--- BIG ELKHART CREEK.prj (project) ---

Proj Title=BIG ELKHART CREEK Base Level Engineering
Current Plan=p01
Default Exp/Contr=0.3,0.1
English Units
Geom File=g01
Flow File=f01
Plan File=p01
Y Axis Title=Elevation
X Axis Title(PF)=Main Channel Distance
X Axis Title(XS)=Station
BEGIN DESCRIPTION:
BIG ELKHART CREEK
END DESCRIPTION:
DSS Export Rating Curves= 0
DSS Export Rating Curve Sorted= 0
DSS Export Volume Flow Curves= 0
DXF OffsetX= 0
DXF OffsetY= 0
DXF ScaleX= 1
DXF ScaleY= 10

--- BIG ELKHART CREEK.p01 (plan) ---

Plan Title=Multiple Run
Short Identifier=Multiple
Geom File=g01
Flow File=f01
Subcritical Flow
K Sum by GR= 0
Std Step Tol= 0.01
Critical Tol= 0.01
Num of Std Step Trials= 20
Max Error Tol= 0.3
Flow Tol Ratio= 0.001
Split Flow NTrial= 30
Split Flow Tol= 0.02
Split Flow Ratio= 0.02
Log Output Level= 0
Friction Slope Method= 1
Unsteady Friction Slope Method= 2
Unsteady Bridges Friction Slope Method= 1
Parabolic Critical Depth
Global Vel Dist=  1 , 1 , 1
Global Log Level= 0
CheckData=True
Encroach Param= -1, 0, 0, 0
BEGIN DESCRIPTION:
Multiple Run
END DESCRIPTION:

--- BIG ELKHART CREEK.f01 (steady flow) ---

Flow Title=Multiple
Program Version=4.10
Number of Profiles= 7
Profile Names=10-year,25-year,50-year,1pct_min,100-year,1pct_plu,500-year
River Rch & RM=BIG ELKHART CREE,Reach-1         ,148528
     762    1043    1278    1151    1557    2105    2316
River Rch & RM=BIG ELKHART CREE,Reach-1         ,146249
    1126    1573    1954    1781    2409    3257    3674
River Rch & RM=BIG ELKHART CREE,Reach-1         ,144667
    1229    1719    2136    1947    2633    3560    4013
River Rch & RM=BIG ELKHART CREE,Reach-1         ,140511
    1258    1759    2186    1991    2692    3641    4102
River Rch & RM=BIG ELKHART CREE,Reach-1         ,137500
    1778    2526    3173    2918    3946    5337    6131
River Rch & RM=BIG ELKHART CREE,Reach-1         ,136106
    2209    3161    3989    3684    4982    6738    7805
River Rch & RM=BIG ELKHART CREE,Reach-1         ,135641
    2209    3161    3989    3684    4982    6738    7805
River Rch & RM=BIG ELKHART CREE,Reach-1         ,131953
    2525    3623    4579    4233    5725    7743    8987
River Rch & RM=BIG ELKHART CREE,Reach-1         ,131111
    2525    3623    4579    4233    5725    7743    8987
River Rch & RM=BIG ELKHART CREE,Reach-1         ,126332
    2815    4055    5139    4762    6440    8710   10158
River Rch & RM=BIG ELKHART CREE,Reach-1         ,124632
    2866    4121    5217    4827    6528    8828   10265
River Rch & RM=BIG ELKHART CREE,Reach-1         ,120716
    4051    5890    7511    6997    9463   12798   15080
River Rch & RM=BIG ELKHART CREE,Reach-1         ,116578
    4112    5972    7612    7085    9582   12959   15247
River Rch & RM=BIG ELKHART CREE,Reach-1         ,112193
    4125    5988    7630    7100    9602   12985   15266
River Rch & RM=BIG ELKHART CREE,Reach-1         ,111330
    4161    6037    7689    7151    9671   13079   15360
River Rch & RM=BIG ELKHART CREE,Reach-1         ,110575
    4202    6089    7748    7199    9736   13167   15432
River Rch & RM=BIG ELKHART CREE,Reach-1         ,106885
    4497    6526    8311    7728   10451   14134   16589
River Rch & RM=BIG ELKHART CREE,Reach-1         ,105514
    4497    6526    8311    7728   10451   14134   16589
River Rch & RM=BIG ELKHART CREE,Reach-1         ,103344
    4896    7115    9073    8444   11420   15444   18161
River Rch & RM=BIG ELKHART CREE,Reach-1         ,102211
    4896    7115    9073    8444   11420   15444   18161
River Rch & RM=BIG ELKHART CREE,Reach-1         ,98935
    4987    7247    9241    8600   11631   15729   18492
River Rch & RM=BIG ELKHART CREE,Reach-1         ,96231
    5019    7289    9288    8638   11682   15798   18548
River Rch & RM=BIG ELKHART CREE,Reach-1         ,89967
    5057    7337    9345    8686   11747   15886   18629
River Rch & RM=BIG ELKHART CREE,Reach-1         ,85110
    5096    7397    9423    8760   11846   16021   18795
River Rch & RM=BIG ELKHART CREE,Reach-1         ,84703
    7100   10386   13305   12430   16811   22734   26926
River Rch & RM=BIG ELKHART CREE,Reach-1         ,83378
    7100   10386   13305   12430   16811   22734   26926
River Rch & RM=BIG ELKHART CREE,Reach-1         ,83244
    7405   10817   13844   12918   17471   23627   27916
River Rch & RM=BIG ELKHART CREE,Reach-1         ,77144
    7405   10817   13844   12918   17471   23627   27916
River Rch & RM=BIG ELKHART CREE,Reach-1         ,66655
    7481   10920   13968   13027   17618   23826   28120
River Rch & RM=BIG ELKHART CREE,Reach-1         ,63009
    7429   10828   13836   12889   17431   23574   27759
River Rch & RM=BIG ELKHART CREE,Reach-1         ,55052
    7427   10814   13809   12855   17385   23511   27645
River Rch & RM=BIG ELKHART CREE,Reach-1         ,51781
    7454   10838   13825   12856   17387   23514   27588
River Rch & RM=BIG ELKHART CREE,Reach-1         ,50852
    7454   10838   13825   12856   17387   23514   27588
River Rch & RM=BIG ELKHART CREE,Reach-1         ,43918
    7618   11062   14100   13100   17717   23960   28058
River Rch & RM=BIG ELKHART CREE,Reach-1         ,34562
    7637   11082   14117   13107   17726   23972   28036
River Rch & RM=BIG ELKHART CREE,Reach-1         ,33151
    7855   11402   14530   13494   18249   24680   28878
River Rch & RM=BIG ELKHART CREE,Reach-1         ,28830
    7855   11402   14530   13494   18249   24680   28878
River Rch & RM=BIG ELKHART CREE,Reach-1         ,26451
    7838   11369   14480   13440   18177   24582   28731
River Rch & RM=BIG ELKHART CREE,Reach-1         ,21557
   11880   17341   22193   20689   27980   37840   44582
Boundary for River Rch & Prof#=BIG ELKHART CREE,Reach-1         , 1
Up Type= 0
Dn Type= 3
Dn Slope=0.001
Boundary for River Rch & Prof#=BIG ELKHART CREE,Reach-1         , 2
Up Type= 0
Dn Type= 3
Dn Slope=0.001
Boundary for River Rch & Prof#=BIG ELKHART CREE,Reach-1         , 3
Up Type= 0
Dn Type= 3
Dn Slope=0.001
Boundary for River Rch & Prof#=BIG ELKHART CREE,Reach-1         , 4
Up Type= 0
Dn Type= 3
Dn Slope=0.001
Boundary for River Rch & Prof#=BIG ELKHART CREE,Reach-1         , 5
Up Type= 0
Dn Type= 3
Dn Slope=0.001
Boundary for River Rch & Prof#=BIG ELKHART CREE,Reach-1         , 6
Up Type= 0
Dn Type= 3
Dn Slope=0.001
Boundary for River Rch & Prof#=BIG ELKHART CREE,Reach-1         , 7
Up Type= 0
Dn Type= 3
Dn Slope=0.001
DSS Import GetInterval= 0
DSS Import GetPeak= 0
DSS Import FillOption= 0

--- BIG ELKHART CREEK.g01 (geometry) ---

Geom Title=Existing Conditions
Program Version=4.10

River Reach=BIG ELKHART CREE,Reach-1
Reach XY= 30
       3798339.5       10562881.      3795904.25       10558020.
      3796903.75       10554770.        3796288.       10551890.
        3794247.       10551025.      3790758.75       10547137.
      3789576.25       10543521.        3784433.       10537087.
       3776909.5       10535801.      3776348.25       10536567.
      3769957.25       10537345.      3768555.75       10539103.
        3764780.       10540191.      3755574.25       10532813.
       3754616.5       10528582.       3752719.5       10526080.
       3753898.5       10522181.        3753197.       10519027.
       3754290.5       10517185.        3752364.       10514435.
       3755447.5       10507540.      3755029.75       10505041.
       3753871.5       10503984.      3754721.25       10502724.
        3753892.       10499716.      3754778.25       10498251.
        3752414.       10495434.       3752252.5       10493983.
      3750939.25       10493873.      3749376.12     10491846.09

Type RM Length L Ch R = 1 ,148528  ,453,453,453
BEGIN DESCRIPTION:
BIG ELKHART CREEK 198.0
END DESCRIPTION:
XS GIS Cut Line= 2
      3798723.41     10562333.82      3797844.95     10562802.56
#Sta/Elev= 30
    4443  449.03  4493.4  448.21    4504  449.02  4509.6  447.89  4560.7  446.82
  4591.8  444.05    4708  442.04  4730.7  440.21  4745.5  440.34  4805.7  434.75
  4833.3  429.43  4855.4  426.78  4865.9  424.07  4913.1  417.78  4931.8  414.12
    4946  414.25  4958.2   412.2  4994.6  410.91  4997.4  410.41  5000.6  410.91
    5048  411.37  5057.8   413.8  5138.7   425.4  5161.4  427.61  5167.6  429.44
    5179  430.05  5227.8  434.25  5255.4  438.59  5321.3  443.39  5438.7  446.05
#Mann= 6 ,-1 , 0
    4443     .16       0  4913.1     .12       0  4958.2     .16       0
  4994.6     .07       0  5000.6     .16       0    5179     .05       0
Bank Sta=4946,5057.8
XS Rating Curve= 0 ,0
Exp/Cntr=0.3,0.1

Type RM Length L Ch R = 1 ,148075  ,295,295,295
BEGIN DESCRIPTION:
BIG ELKHART CREEK 197.0
END DESCRIPTION:
XS GIS Cut Line= 3
      3798244.24     10562059.52      3797949.12     10562253.95
      3797647.91     10562676.34
#Sta/Elev= 30
  4565.5  439.67  4612.6  439.07  4618.9  437.82  4667.2  434.82  4736.1  431.24
  4799.2  425.04  4808.3  425.24  4822.5  422.27  4830.2  422.08  4850.5   420.1
  4858.4  420.52  4871.5   418.2  4907.2  415.15  4918.9  413.87  4923.6   412.4
  4938.3  410.35  4977.1  409.98  4979.8  409.48  4983.1  409.98  5037.1  410.09
    5060  413.25  5074.6  415.62    5087   415.8  5131.3  422.12  5152.2  423.78
  5217.3  432.32  5238.2  433.53  5259.1     436    5339  440.25  5437.7  443.14
#Mann= 7 ,-1 , 0
  4565.5     .05       0  4667.2     .16       0  4830.2     .05       0
  4907.2     .16       0  4977.1     .07       0  4983.1     .16       0
  5074.6     .05       0
Bank Sta=4923.6,5060
XS Rating Curve= 0 ,0
Exp/Cntr=0.3,0.1

Type RM Length L Ch R = 1 ,147780  ,466,466,466
BEGIN DESCRIPTION:
BIG ELKHART CREEK 196.0
END DESCRIPTION:
XS GIS Cut Line= 3
      3797942.16     10561983.13      3797744.26     10562080.34
      3797300.95     10562506.33
#Sta/Elev= 30
  4643.8  437.44  4689.7  436.89  4734.7  434.52  4746.9  432.44  4779.7  429.76
  4813.8  424.83  4824.6  424.67  4867.8  419.52  4874.5  417.89    4910  414.15
  4916.9  412.32  4924.1  410.25    4939  408.28  4959.4  408.86  4963.6  407.77
  4966.3  407.27  4969.6  407.77  5058.4  409.35  5065.4  411.26  5084.9  412.78
  5100.9  413.52    5122  416.45  5192.7  422.74  5305.9  430.53  5376.7  432.54
    5405  431.92  5426.1  432.82  5447.4   432.3  5454.4  433.42  5479.1  433.06
#Mann= 5 ,-1 , 0
  4643.8     .05       0    4939     .16       0  4963.6     .07       0
  4969.6     .16       0  5084.9     .05       0
Bank Sta=4916.9,5065.4
XS Rating Curve= 0 ,0
Exp/Cntr=0.3,0.1

Type RM Length L Ch R = 1 ,147314  ,118,118,118
BEGIN DESCRIPTION:
Mapping XS 522f206a
END DESCRIPTION:
XS GIS Cut Line= 4
       3797950.3      10561897.8      3797450.32     10561852.66
      3797280.18     10561849.19      3796856.56     10562043.64
#Sta/Elev= 30
  4391.2  436.31  4522.4  430.93  4562.6  427.46  4652.9  423.69  4693.1  422.37
  4743.3  422.75  4793.5  421.09  4840.2  417.76  4861.9  415.14    4867  415.72
  4896.1  413.37  4933.9  408.76  4943.9  408.85  4990.9  406.47  4993.7  405.97
  4996.9  406.47    5034  406.51  5066.5  407.41  5073.6  408.85    5086  409.47
  5096.6  411.35    5119  412.14  5207.1   423.2  5291.5  429.76    5343  431.06
  5350.1  432.61  5369.1  433.43    5412  435.19  5440.5  434.91  5529.5  437.38
#Mann= 6 ,-1 , 0
  4391.2     .05       0  4840.2     .16       0  4990.9     .07       0
  4996.9     .16       0    5034     .05       0  5369.1     .16       0
Bank Sta=4943.9,5073.6
XS Rating Curve= 0 ,0
Exp/Cntr=0.3,0.1

Type RM Length L Ch R = 1 ,147196  ,429,429,429
BEGIN DESCRIPTION:
BIG ELKHART CREEK 195.0
END DESCRIPTION:
XS GIS Cut Line= 4
      3798193.39     10561745.02      3797450.32     10561734.61
      3797301.01     10561734.61       3796833.4     10561814.27
#Sta/Elev= 30
  4138.1  432.62  4230.7   427.1  4381.9  417.19  4401.9  417.77  4428.4  415.93
  4527.3  415.04  4631.9  415.17  4651.9  412.52    4872  414.65    4932  408.78
  4958.4  407.67    4972  407.43    5009  405.48  5011.7  404.98    5015  405.48
  5042.1  408.25  5082.7  407.57    5103  408.95  5150.9  416.07  5155.9  415.17
    5174  418.91  5223.3  423.98  5234.9  426.18  5265.3  427.32  5271.3  430.17
  5285.6  429.66  5331.5  433.15  5451.9  437.62    5494  437.61  5504.9  438.21
#Mann= 9 ,-1 , 0
  4138.1     .05       0  4230.7      .1       0  4428.4     .05       0
  4527.3     .16       0  4958.4     .05       0    5009     .04       0
    5015     .05       0  5223.3     .16       0    5494     .05       0
Bank Sta=4972,5042.1
XS Rating Curve= 0 ,0
Exp/Cntr=0.3,0.1

Type RM Length L Ch R = 1 ,146767  ,518,518,518
BEGIN DESCRIPTION:
BIG ELKHART CREEK 194.0
END DESCRIPTION:
XS GIS Cut Line= 3
       3797657.5     10561281.72      3797299.82     10561299.09
      3796763.07     10561551.88
#Sta/Elev= 30
  4501.8  438.43  4639.9  432.27    4750  424.21  4777.3  421.21  4782.3  421.85
  4804.3  418.86  4869.9  412.99  4882.2  410.44  4892.7  410.02  4915.4  407.34
    4921  405.32  4937.5  404.02  4943.8  402.55  4986.4  401.02  4989.2  400.52
  4992.4  401.02  5025.9  402.94    5035  403.06  5070.2  408.07  5103.3  410.53
  5108.9  412.23  5147.5  413.59    5160   415.7  5169.6  415.93  5177.2  418.96
    5200  422.09  5291.2  422.73  5313.3  424.63    5325  428.52  5453.2   435.4
#Mann= 4 ,-1 , 0
  4501.8      .1       0  4804.3     .16       0  4986.4     .07       0
  4992.4     .16       0
Bank Sta=4937.5,5025.9
XS Rating Curve= 0 ,0
Exp/Cntr=0.3,0.1

Type RM Length L Ch R = 1 ,146249  ,401,401,401
BEGIN DESCRIPTION:
BIG ELKHART CREEK 193.0
END DESCRIPTION:
XS GIS Cut Line= 3
      3797282.42     10560698.42      3796761.62     10561052.56
       3796581.1     10561174.06
#Sta/Elev= 30
  4508.7  432.71  4642.2  425.34  4669.3  424.93  4684.1  423.14  4705.6  422.19
  4741.9  417.51  4821.8  413.39  4843.4  410.75  4857.7  409.68  4863.7  410.22
  4872.6  408.52  4965.5  397.92  4980.4  397.49  4986.4  396.61  4992.3  394.39
  4995.1  393.89  4998.3  394.39  5001.4  394.88  5007.9  399.39  5031.3  399.96
  5052.2  402.28  5094.2  409.42  5103.1  409.83  5136.7  415.43    5153  416.66
  5166.1  419.27  5274.1  430.61  5286.5  430.44  5333.8  433.86  5356.1  433.54
#Mann= 4 ,-1 , 0
  4508.7     .05       0  4843.4     .16       0  4992.3     .07       0
  4998.3     .16       0
Bank Sta=4980.4,5007.9
XS Rating Curve= 0 ,0
Exp/Cntr=0.3,0.1

Type RM Length L Ch R = 1 ,145848  ,442,442,442
BEGIN DESCRIPTION:
BIG ELKHART CREEK 192.0
END DESCRIPTION:
XS GIS Cut Line= 3
      3797285.89     10560549.09       3796601.9     10560653.25
      3796387.53      10560926.4
#Sta/Elev= 30
  4382.1  434.61  4499.7  427.32  4530.1  424.09    4611  420.16  4687.6  413.18
  4692.6  414.37  4704.2  413.94  4833.5  408.41  4888.4  403.14  4914.4  398.71
    4965  396.86  4985.3  395.12  4992.4  391.88  4995.1  391.38  4998.4  391.88
  5025.7  396.11  5066.2  395.31  5072.6  400.37  5101.9  402.97  5108.3  405.92
  5145.3  409.61  5151.6  411.92  5180.5  415.47  5222.6  418.04  5236.6  420.18
  5259.2  421.06  5273.5   419.8  5286.3  420.78  5294.4  423.11  5421.2  426.44
#Mann= 4 ,-1 , 0
  4382.1     .05       0  4704.2     .16       0  4992.4     .07       0
  4998.4     .16       0
Bank Sta=4965,5025.7
XS Rating Curve= 0 ,0
Exp/Cntr=0.3,0.1

Type RM Length L Ch R = 1 ,145406  ,739,739,739
BEGIN DESCRIPTION:
BIG ELKHART CREEK 191.0
END DESCRIPTION:
XS GIS Cut Line= 3
      3797324.11     10560392.83      3796299.82     10560094.23
      3795943.41     10560163.43
#Sta/Elev= 30
  4406.3  436.05  4568.9  427.19  4651.9  419.25  4680.2  418.03  4743.5  409.26
  4806.8  400.71  4817.2  400.48  4848.5  395.36    4911  394.23  4952.6  391.63
  4968.9  393.41  4994.3  389.56  5002.4  390.37  5015.1  393.95  5079.8   395.3
  5108.1  391.93  5116.3  388.76    5119  388.26  5122.3  388.76  5140.1  395.65
  5180.3  393.76  5224.2  397.43  5317.2  399.17  5358.1  401.69  5478.4  405.26
  5514.2  408.34  5524.4  407.48  5633.5  410.76  5768.9  416.27  5836.3  416.93
#Mann= 5 ,-1 , 0
  4406.3     .05       0  4568.9      .1       0  4743.5     .16       0
  5116.3     .07       0  5122.3     .16       0
Bank Sta=4911,5140.1
XS Rating Curve= 0 ,0
Exp/Cntr=0.3,0.1

Type RM Length L Ch R = 1 ,144667  ,494,494,494
BEGIN DESCRIPTION:
BIG ELKHART CREEK 190.0
END DESCRIPTION:
XS GIS Cut Line= 3
      3797181.76      10559785.2      3796355.37     10559802.56
      3795955.31     10559885.33
#Sta/Elev= 30
  4312.2  441.82  4404.4  438.21  4574.4   426.2  4634.4  423.24  4654.4  421.36
  4664.4  416.91  4674.4  418.72  4694.4   418.2  4774.5  409.51  4794.5  407.04
  4804.5  404.36  4832.5  401.36  4904.5     392  4934.5  390.81  4944.5  392.26
  4984.5  392.31  4996.4  386.24  5001.5  385.95  5004.3  385.45  5007.5  385.95
  5014.5  390.25  5044.5  392.94  5138.8  398.07  5150.8  400.01  5236.6  406.78
  5251.2  406.38  5267.2  408.36  5301.6  409.62  5497.1  417.87  5547.3  418.77
#Mann= 6 ,-1 , 0
  4312.2     .16       0  4832.5     .12       0  4996.4     .16       0
  5001.5     .07       0  5007.5     .16       0  5301.6     .05       0
Bank Sta=4984.5,5044.5
XS Rating Curve= 0 ,0
Exp/Cntr=0.3,0.1

Type RM Length L Ch R = 1 ,144173  ,543,543,543
BEGIN DESCRIPTION:
BIG ELKHART CREEK 189.0
END DESCRIPTION:
XS GIS Cut Line= 3
      3796806.74     10559288.68       3796265.1     10559455.34
      3795810.27     10559424.09
#Sta/Elev= 30
  4477.8  429.42  4538.4  423.75  4565.8  423.46  4579.4  420.73  4674.4  415.69
  4757.3  408.17  4851.5  403.32  4903.3  398.19  4914.2  398.55  4923.7  396.43
  4966.5  391.84  4979.1  389.31  4987.5  384.07  4994.9  383.07  4997.7  382.57
  5000.9  383.07  5006.6  385.86  5011.8  383.78  5018.9  388.65  5029.3  390.37
  5080.1  390.62  5120.2  392.61  5129.9  394.69  5180.3  405.38  5220.4  408.66
  5337.1  413.79  5430.9  415.03  5450.9  417.47    5461  416.64  5500.4  419.43
#Mann= 5 ,-1 , 0
  4477.8     .16       0  4923.7     .12       0  4994.9     .07       0
  5000.9     .12       0  5129.9     .16       0
Bank Sta=4966.5,5029.3
XS Rating Curve= 0 ,0
Exp/Cntr=0.3,0.1

Type RM Length L Ch R = 1 ,143630  ,447,447,447
BEGIN DESCRIPTION:
BIG ELKHART CREEK 188.0
END DESCRIPTION:
XS GIS Cut Line= 2
      3796897.08      10559035.2      3795752.93     10559010.93
#Sta/Elev= 30
  4475.7  440.96  4643.2  429.76  4743.2  421.17  4753.2  421.08  4763.2  419.21
  4790.4  417.72  4833.2  414.16  4873.3  409.41  4903.3     404  4913.3  400.05
  4933.3  396.14  4983.3  390.69  4993.3  386.59  5000.3  381.97    5003  381.47
  5006.3  381.97  5013.3  384.82  5033.3   386.9  5103.3  387.85  5133.3  386.87
  5153.3  387.98  5203.3  394.45  5273.3   399.9  5304.3  403.51  5383.4  408.98
  5413.4  411.95  5463.4  413.44  5483.4  412.33  5503.4  415.28  5620.1   421.6
#Mann= 5 ,-1 , 0
  4475.7     .16       0  4790.4     .12       0  5000.3     .07       0
  5006.3     .12       0  5304.3     .16       0
Bank Sta=4983.3,5033.3
XS Rating Curve= 0 ,0
Exp/Cntr=0.3,0.1

Type RM Length L Ch R = 1 ,143183  ,438,438,438
BEGIN DESCRIPTION:
BIG ELKHART CREEK 187.0
END DESCRIPTION:
XS GIS Cut Line= 4
      3796799.87     10558806.04      3796338.01     10558674.09
       3796140.1     10558653.25      3795765.14     10558750.47
#Sta/Elev= 30
  4405.6  430.33  4530.7  424.21  4680.2  412.94  4734.9   405.2  4773.9  401.87
  4790.7   398.5  4807.7  393.32  4812.9  393.55  4832.3  389.43  4846.7  388.05
  4853.1  385.12  4873.9  386.42  4883.9  384.19  4904.4  385.65  4975.4  385.39
  4991.9  381.96  4994.7  381.46  4997.9  381.96    5015  385.01  5055.3   384.3
  5106.1   385.3  5126.8   383.7  5132.2   385.4  5188.8  387.64  5335.1  407.79
  5392.3  413.58  5402.1  414.51  5411.1  416.89  5436.7   419.2  5472.3  420.73
#Mann= 6 ,-1 , 0
  4405.6     .16       0  4680.2     .12       0  4991.9     .07       0
  4997.9     .12       0  5392.3     .05       0  5402.1     .16       0
Bank Sta=4975.4,5015
XS Rating Curve= 0 ,0
Exp/Cntr=0.3,0.1

Type RM Length L Ch R = 1 ,142745  ,574,574,574
BEGIN DESCRIPTION:
BIG ELKHART CREEK 186.0
END DESCRIPTION:
XS GIS Cut Line= 3
      3796553.29     10558240.06      3796244.26     10558260.89
      3795650.49     10558569.93
#Sta/Elev= 30
  4516.7  417.39  4630.6  411.53  4739.6  401.84  4821.1  397.06  4826.3  395.53
  4849.4  392.96  4856.3  392.01  4919.3  382.53  4991.2  382.65  5004.7  379.67
  5007.5  379.17  5010.7  379.67  5013.3  381.58  5023.3  382.63  5237.5  383.69
  5250.8  384.93  5260.1  388.19  5267.3  388.62  5295.1  395.77  5305.2  397.23
  5311.5  400.34  5333.6   405.1  5350.1  406.69  5361.5  409.83  5375.1  411.79
  5395.7  414.52  5406.6  416.34  5438.5  417.56  5444.1   418.9  5495.8  419.79
#Mann= 8 ,-1 , 0
  4516.7     .16       0  4739.6     .12       0  4849.4     .16       0
  4856.3     .12       0  5004.7     .07       0  5010.7     .12       0
  5375.1     .16       0  5395.7     .05       0
Bank Sta=4991.2,5023.3
XS Rating Curve= 0 ,0
Exp/Cntr=0.3,0.1

Type RM Length L Ch R = 1 ,142171  ,305,305,305
BEGIN DESCRIPTION:
BIG ELKHART CREEK 185.0
END DESCRIPTION:
XS GIS Cut Line= 3
      3796334.53     10557868.53      3795820.65     10557931.03
      3795553.96     10558377.83
#Sta/Elev= 30
  4553.3  406.24  4557.5  406.24  4598.6  405.23  4679.1  400.86  4719.4  396.78
  4725.3  395.05  4749.7   390.8  4810.1  384.21  4820.2  384.73  4829.8  382.86
  4870.5  379.29  4942.9  379.04  4981.4  380.25  4998.5  378.77  5001.2  378.27
  5004.5  378.77  5019.6  380.24  5144.1  380.11    5233  380.53  5275.8  383.71
  5312.8  389.52  5318.6  392.38  5349.5  396.76  5361.4  399.96  5384.4   401.7
  5398.4  406.02  5429.6  407.91  5435.4  407.33  5472.4  411.94  5591.3   413.5
#Mann= 7 ,-1 , 0
  4553.3     .16       0  4557.5     .12       0  4725.3     .16       0
  4829.8     .12       0  4998.5     .07       0  5004.5     .12       0
  5144.1     .16       0
Bank Sta=4981.4,5019.6
XS Rating Curve= 0 ,0
Exp/Cntr=0.3,0.1

Type RM Length L Ch R = 1 ,141866  ,657,657,657
BEGIN DESCRIPTION:
BIG ELKHART CREEK 184.0
END DESCRIPTION:
XS GIS Cut Line= 3
      3796682.93     10557824.88       3795752.4     10557658.22
      3795523.92     10557436.66
#Sta/Elev= 30
  4303.9  422.25  4414.8  416.68  4542.3  412.52  4632.4  408.64  4662.8  408.96
  4744.1  404.79  4764.4  401.57  4811.4  399.14  4825.4  395.44    4841  394.29
  4947.3  379.72  4998.1  378.21  5018.4  379.44    5094  379.14  5167.8  378.08
  5170.5  377.58  5173.8  378.08    5181  379.26  5251.4  380.34  5285.1  384.12
  5313.4  389.07  5327.6  395.52  5363.1   400.8    5370  404.66  5377.2   404.9
  5398.3  410.33  5430.4  414.03    5469   415.8  5504.3  420.26  5567.5  422.28
#Mann= 7 ,-1 , 0
  4303.9      .1       0  4542.3     .16       0    4841     .12       0
    5094     .16       0  5167.8     .07       0  5173.8     .16       0
  5430.4     .05       0
Bank Sta=4947.3,5181
XS Rating Curve= 0 ,0
Exp/Cntr=0.3,0.1

Type RM Length L Ch R = 1 ,141209  ,569,569,569
BEGIN DESCRIPTION:
BIG ELKHART CREEK 183.0
END DESCRIPTION:
XS GIS Cut Line= 3
      3796549.79     10557615.04      3796088.01     10557233.11
      3795742.73     10557181.32
#Sta/Elev= 30
  4465.6  410.97  4511.8   407.8    4547  403.24  4561.3  402.78  4628.1   393.1
  4703.3  384.21  4711.2   384.4    4732  380.91  4760.6  378.52  4767.1  378.93
  4810.1  375.74  4891.8  375.69  4894.5  375.19  4897.8  375.69  4902.6  376.66
  4952.1  375.96  4966.5  376.86  5103.7  377.26  5113.5  378.39  5144.1  377.32
  5154.2  381.23  5187.7  386.21  5204.8  392.74  5214.9   393.7  5245.3  403.12
  5256.8  405.57  5285.7  410.89  5320.8  414.51  5336.3  418.02    5414  420.55
#Mann= 4 ,-1 , 0
  4465.6      .1       0  4628.1     .16       0  4891.8     .07       0
  4897.8     .16       0
Bank Sta=4767.1,5113.5
XS Rating Curve= 0 ,0
Exp/Cntr=0.3,0.1

Type RM Length L Ch R = 1 ,140640  ,129,129,129
BEGIN DESCRIPTION:
BIG ELKHART CREEK 182.0
END DESCRIPTION:
XS GIS Cut Line= 6
      3797276.71     10556675.58      3796964.21     10556540.16
      3796783.65     10556550.58      3796457.26      10556772.8
      3796196.84     10556831.83      3795790.58     10557147.81
#Sta/Elev= 30
    3976  433.65  4252.2  422.89  4277.8  418.42  4316.4  414.82  4465.2   412.3
  4542.2  410.17  4550.3  405.98  4571.1  403.77  4584.8  397.81  4591.2  397.96
  4642.2  386.96  4685.1  384.07  4699.5  377.89  4714.2  376.69  4800.5  374.66
  4945.3  374.84  4971.5  375.45  4978.5  374.32  4981.2  373.82  4984.5  374.32
  5001.5  375.83  5140.2  375.61  5233.9  387.07  5368.8  396.27  5397.7  403.09
  5418.5  402.63  5511.7   410.9  5541.3  410.63    5576  416.09  5680.2  418.89
#Mann= 11 ,-1 , 0
    3976     .05       0  4277.8      .1       0  4465.2     .16       0
  4584.8     .05       0  4591.2     .16       0  4714.2     .05       0
  4800.5     .12       0  4945.3     .05       0  4978.5     .04       0
  4984.5     .05       0  5541.3     .16       0
Bank Sta=4971.5,5001.5
XS Rating Curve= 0 ,0
Exp/Cntr=0.3,0.1

Type RM Length L Ch R = 1 ,140511  ,547,547,547
BEGIN DESCRIPTION:
BIG ELKHART CREEK 181.0
END DESCRIPTION:
XS GIS Cut Line= 6
      3797339.24     10556439.47      3796759.34      10556397.8
      3796603.09     10556481.13      3796509.34     10556651.27
      3796228.09     10556692.94      3795697.35     10557015.54
#Sta/Elev= 30
  3899.6  430.38  4149.9  413.54    4180  407.04    4200  410.19  4220.1  410.03
  4410.5  394.15  4513.2  392.49  4523.3  394.17  4563.1  393.45  4579.4   388.9
  4639.4  380.86  4645.2  375.28    4686  374.03  4756.3  375.84  4912.7  373.03
  4922.8   374.7  4990.6  372.38  4993.3  371.88  4996.6  372.38  5094.7  374.27
  5192.9  376.04  5285.2  386.89  5375.3  398.91  5390.2  398.97  5396.6  401.99
  5433.2  402.57  5460.8  409.64  5548.9  416.11  5695.3  419.35  5757.8  417.98
#Mann= 7 ,-1 , 0
  3899.6     .16       0  4513.2     .05       0  4523.3     .16       0
    4686     .05       0  4990.6     .04       0  4996.6     .05       0
  5285.2     .16       0
Bank Sta=4922.8,5094.7
XS Rating Curve= 0 ,0
Exp/Cntr=0.3,0.1

Type RM Length L Ch R = 1 ,139964  ,714,714,714
BEGIN DESCRIPTION:
BIG ELKHART CREEK 180.0
END DESCRIPTION:
XS GIS Cut Line= 2
      3797060.21     10556174.09      3795605.36     10556271.31
#Sta/Elev= 30
    4147  427.31    4308  410.73    4348  405.07  4368.1  401.31  4378.1  395.94
  4408.2  387.64  4438.2  385.47  4458.3  382.39  4463.4  380.11  4468.4  380.86
  4488.4  374.31  4571.5  372.02  4698.8  369.23  4913.8  370.32  4919.3   368.6
  4989.5  368.96  4996.5   367.6  4999.2   367.1  5002.5   367.6  5119.8  371.32
  5179.9  374.73  5209.1  380.42    5220  380.87  5272.4  391.95  5330.2  401.71
  5364.3  403.35  5371.7  406.02  5400.4   407.2  5500.6     417  5605.1  421.76
#Mann= 6 ,-1 , 0
    4147     .16       0  4571.5     .12       0  4996.5     .07       0
  5002.5     .12       0  5272.4     .16       0  5371.7     .05       0
Bank Sta=4913.8,5119.8
XS Rating Curve= 0 ,0
Exp/Cntr=0.3,0.1

Type RM Length L Ch R = 1 ,139250  ,425,425,425
BEGIN DESCRIPTION:
BIG ELKHART CREEK 179.0
END DESCRIPTION:
XS GIS Cut Line= 2
      3797084.53      10555910.2      3795959.56     10555757.42
#Sta/Elev= 30
  4485.8  419.88  4519.5  416.62  4524.6  417.58  4591.7  408.43    4597  406.48
  4611.9  405.57    4622  402.04  4682.5  390.09  4692.6  389.58  4712.8  384.06
  4753.2  377.91  4783.4  375.76  4864.2  366.25  4965.9  366.18  4985.3  366.03
  4992.4  365.27  4995.1  364.77  4998.4  365.27  5005.4  365.96  5146.7   367.4
  5257.7  366.53  5269.5  367.25  5277.9  369.85  5328.4   371.3  5356.4   376.9
  5414.5  387.39  5486.9  398.43  5570.6  405.54  5580.7  407.42  5621.1  408.99
#Mann= 5 ,-1 , 0
  4485.8     .16       0  4965.9     .12       0  4992.4     .07       0
  4998.4     .12       0  5356.4     .16       0
Bank Sta=4985.3,5005.4
XS Rating Curve= 0 ,0
Exp/Cntr=0.3,0.1

Type RM Length L Ch R = 1 ,138825  ,406,406,406
BEGIN DESCRIPTION:
BIG ELKHART CREEK 178.0
END DESCRIPTION:
XS GIS Cut Line= 3
      3797119.25     10555750.46       3796789.4     10555479.64
      3796185.23     10555431.03
#Sta/Elev= 30
  4449.7  425.21  4549.4  417.51  4570.2  413.64  4591.6  412.65  4683.6  402.15
  4691.5  399.83  4712.3   397.6  4720.2  394.36  4726.7  394.33  4733.9  389.98
  4747.5  387.92  4755.4  384.42  4769.7  382.08  4776.2  382.96  4784.1  378.88
  4790.5  379.23  4798.4  375.73  4898.9  365.91  4996.7  362.92  5003.7  362.79
  5006.4  362.29  5009.7  362.79  5016.7  363.22    5212  363.92  5237.4  365.49
  5267.5  371.08  5297.6  374.33  5317.7   378.8  5377.9  386.57  5482.6   393.5
#Mann= 5 ,-1 , 0
  4449.7     .16       0  4898.9     .12       0  5003.7     .07       0
  5009.7     .12       0    5212     .16       0
Bank Sta=4996.7,5016.7
XS Rating Curve= 0 ,0
Exp/Cntr=0.3,0.1

Type RM Length L Ch R = 1 ,138419  ,480,480,480
BEGIN DESCRIPTION:
BIG ELKHART CREEK 177.0
END DESCRIPTION:
XS GIS Cut Line= 2
      3797248.93     10555265.86      3796113.17     10554962.41
#Sta/Elev= 30
  4396.7  421.44  4427.1  420.17  4499.5  414.18  4509.9  414.41  4515.3  412.35
  4540.9  410.91  4582.3  406.21  4623.7  398.98  4644.4  393.24  4675.6  389.38
  4696.2  384.43  4705.3  379.95  4716.9  378.85  4785.4  366.02  4799.7  365.47
  4825.1  363.36  4841.1  361.79  4931.2  361.37    4934  360.87  4937.2  361.37
  5027.4  361.58  5055.6  365.72  5063.8  367.52  5100.8   372.3  5175.8  378.45
  5285.7  383.09  5290.8  382.26    5371  383.09  5493.2  390.49  5572.3  392.34
#Mann= 5 ,-1 , 0
  4396.7     .16       0  4825.1     .12       0  4931.2     .07       0
  4937.2     .12       0  5063.8     .16       0
Bank Sta=4799.7,5055.6
XS Rating Curve= 0 ,0
Exp/Cntr=0.3,0.1

Type RM Length L Ch R = 1 ,137939  ,439,439,439
BEGIN DESCRIPTION:
BIG ELKHART CREEK 176.0
END DESCRIPTION:
XS GIS Cut Line= 3
      3797149.63     10555010.21      3796899.61     10554710.19
      3796099.58     10554810.19
#Sta/Elev= 30
  4600.9  400.89  4614.6  397.86    4679  390.12  4700.5     385    4707  381.85
  4756.8   372.5  4803.6  369.03    4864   364.2    4927  362.42  4949.1  363.78
    4970  362.19  5011.6  361.57  5034.3  362.49  5041.8  361.62    5062  363.43
  5172.8  362.85  5182.9  363.76  5195.5  362.55  5213.2  363.18  5230.1  362.01
  5250.5  361.46  5253.2  360.96  5256.5  361.46  5344.2  362.84  5432.3  369.68
  5444.9  369.67  5465.1  372.16  5565.9  377.65  5674.2  386.86  5797.7   393.5
#Mann= 7 ,-1 , 0
  4600.9     .16       0  4756.8     .12       0  4803.6     .16       0
    4864     .12       0  5230.1     .16       0  5250.5     .07       0
  5256.5     .16       0
Bank Sta=4949.1,5062
XS Rating Curve= 0 ,0
Exp/Cntr=0.3,0.1

Type RM Length L Ch R = 1 ,137500  ,436,436,436
BEGIN DESCRIPTION:
BIG ELKHART CREEK 175.0
END DESCRIPTION:
XS GIS Cut Line= 3
      3797349.64     10554060.18      3796799.61     10554310.19
      3796349.58     10554560.21
#Sta/Elev= 30
  4379.8  403.52  4468.8   395.8  4500.7  391.92  4514.9  391.42  4555.6  386.37
  4635.8  379.07  4643.5  377.37  4658.8  376.22  4665.4  374.15  4687.4  372.67
    4705  367.78    4728  364.86  4751.1  363.09  4756.6  363.64  4764.3   362.2
  4781.2  361.95  4866.5  361.79  5109.8  362.31  5132.7   361.5    5167  362.26
  5178.9  361.05  5181.6  360.55  5184.9  361.05  5189.9  364.17  5190.4  364.22
  5203.6  365.18  5235.7  371.05  5247.1  371.86  5441.6  379.74  5498.8  383.55
#Mann= 6 ,-1 , 0
  4379.8     .05       0  4781.2     .07       0  4866.5     .12       0
  5178.9     .07       0  5184.9     .12       0  5190.4     .05       0
Bank Sta=4756.6,5189.9
XS Rating Curve= 0 ,0
Exp/Cntr=0.3,0.1

Type RM Length L Ch R = 1 ,137064  ,517,517,517
BEGIN DESCRIPTION:
BIG ELKHART CREEK 174.0
END DESCRIPTION:
XS GIS Cut Line= 3
      3797349.56     10553910.19      3796749.61     10553910.19
      3796349.57     10553810.18
#Sta/Elev= 30
  4394.7  403.74  4424.7  400.84  4464.7  394.32  4504.7  389.55  4604.7  379.09
  4634.7  377.12  4664.7  371.02  4684.7  368.75  4744.7  368.31  4774.7  364.66
  4854.7  357.73  4914.7  356.76  4924.7   357.6  4926.5  357.57  5056.1  356.54
  5058.8  356.04  5062.1  356.54    5127  356.62  5190.5   358.5  5223.6  358.99
    5228  359.32  5265.2  360.49  5283.3  362.49  5301.3  367.07  5314.2  368.21
  5365.7  376.85    5376  377.17  5383.8  378.92  5388.9  378.17    5407  379.05
#Mann= 7 ,-1 , 0
  4394.7     .05       0  4926.5     .12       0  5056.1     .07       0
  5062.1     .12       0    5127     .07       0  5223.6     .12       0
    5228     .16       0
Bank Sta=4924.7,5190.5
XS Rating Curve= 0 ,0
Exp/Cntr=0.3,0.1

Type RM Length L Ch R = 1 ,136547  ,441,441,441
BEGIN DESCRIPTION:
BIG ELKHART CREEK 173.0
END DESCRIPTION:
XS GIS Cut Line= 3
      3797355.34     10553875.45      3796730.37     10553455.34
      3796025.48     10553569.93
#Sta/Elev= 30
    4307  402.68  4502.7  381.98  4553.6  378.58  4625.6  371.26  4826.6  357.56
  4892.3  355.46  4919.7  355.25  4928.4  356.43    4937  355.45  4997.6  354.89
  5000.4  354.39  5003.6  354.89  5032.1   355.4  5101.3  355.18  5111.5  356.14
  5134.2  355.83  5154.9  356.35  5233.1  355.42  5431.8  367.55  5455.9  367.39
  5493.4  372.38  5516.7  372.37  5554.9  376.53    5560  375.78  5597.8  380.39
  5638.3  382.88  5678.1  387.63  5749.7  392.18  5759.7  393.92  5774.2  394.69
#Mann= 8 ,-1 , 0
    4307     .05       0    4937     .12       0  4997.6     .07       0
  5003.6     .12       0  5032.1     .07       0  5134.2     .12       0
  5154.9     .16       0  5759.7     .08       0
Bank Sta=4928.4,5111.5
XS Rating Curve= 0 ,0
Exp/Cntr=0.3,0.1

Type RM Length L Ch R = 1 ,136106  ,465,465,465
BEGIN DESCRIPTION:
BIG ELKHART CREEK 172.0
END DESCRIPTION:
XS GIS Cut Line= 3
      3797099.62     10552510.17      3796699.61     10553110.19
       3796099.6     10553310.19
#Sta/Elev= 30
  4279.1     385  4337.7   382.2  4385.9  379.89  4487.9  367.41    4503  367.77
  4560.1  361.68  4647.2  358.75  4662.2  355.95  4827.5  355.83    4856  353.93
  4863.5  355.89  4884.6  356.72  4947.7  353.23  4950.4  352.73  4953.7  353.23
  5010.8  355.04  5042.4  353.46  5063.5  354.94  5116.2   353.9  5263.8  362.26
  5284.8  366.45  5305.9  368.37  5369.4  371.53  5400.8  374.48  5442.9   372.4
  5474.6  375.98  5506.2  375.75  5527.3  377.77  5542.8  381.36  5632.7  386.84
#Mann= 7 ,-1 , 0
  4279.1     .05       0  4337.7     .08       0  4385.9     .05       0
  4947.7     .03       0  4953.7     .05       0  5369.4     .08       0
  5542.8     .05       0
Bank Sta=4884.6,5010.8
XS Rating Curve= 0 ,0
Exp/Cntr=0.3,0.1

Type RM Length L Ch R = 1 ,135641  ,462,462,462
BEGIN DESCRIPTION:
BIG ELKHART CREEK 171.0
END DESCRIPTION:
XS GIS Cut Line= 3
      3797049.62     10552260.18      3796549.61     10552710.19
      3795949.61     10553110.19
#Sta/Elev= 30
  4298.9  397.14  4391.2  390.66    4469  381.28  4489.9  380.34  4497.4  378.13
  4525.8  376.32  4532.5  377.22  4560.9  372.86    4568  369.57  4581.8   367.8
  4589.3  364.49  4610.2  362.24  4617.7  358.56  4624.4  360.44  4631.9  357.01
  4652.8  355.69  4660.3  353.67  4979.1  354.94  5000.1  351.72  5015.2  350.83
  5021.2  351.99  5027.2  350.62  5029.9  350.12  5033.2  350.62  5051.2  355.52
  5332.2  367.98  5390.7  374.77  5483.9   377.8  5525.9   382.9  5692.7  394.13
#Mann= 3 ,-1 , 0
  4298.9     .05       0  5027.2     .03       0  5033.2     .05       0
Bank Sta=4979.1,5051.2
XS Rating Curve= 0 ,0
Exp/Cntr=0.3,0.1

Type RM Length L Ch R = 1 ,135179  ,452,452,452
BEGIN DESCRIPTION:
BIG ELKHART CREEK 170.0
END DESCRIPTION:
XS GIS Cut Line= 3
      3796949.62     10551960.18      3796349.61     10552310.19
      3795799.62     10552710.18
#Sta/Elev= 30
  4270.8  397.43  4364.7  389.45  4423.4  382.24  4476.3  374.01  4490.8  373.06
  4497.8   368.9  4513.5  367.09  4525.5  363.63  4606.5   357.8    4621  358.51
  4629.7  356.38  4673.9  352.97  4738.4  349.52  4797.2  350.77  4936.1  350.75
    4979  352.57  4987.5  352.06  4999.1  349.32  5001.9  348.82  5005.1  349.32
  5008.3  351.32  5014.9  351.73    5052  352.16  5058.6  353.98  5123.5  358.35
  5129.7  359.73    5159  360.35  5179.9  363.32  5366.1  374.49  5645.5  395.67
#Mann= 3 ,-1 , 0
  4270.8     .05       0  4999.1     .03       0  5005.1     .05       0
Bank Sta=4979,5014.9
XS Rating Curve= 0 ,0
Exp/Cntr=0.3,0.1

Type RM Length L Ch R = 1 ,134727  ,406,406,406
BEGIN DESCRIPTION:
BIG ELKHART CREEK 169.0
END DESCRIPTION:
XS GIS Cut Line= 3
      3796649.58      10551710.2      3796299.61     10551910.19
      3795699.62     10552510.18
#Sta/Elev= 30
    4587  381.11  4659.7  375.77  4718.7  365.91  4740.3  363.38  4756.1  359.28
  4771.2  359.98  4777.7  357.56  4805.8  355.72  4842.5  351.87  4864.1   352.7
  4874.2  351.17  4879.9  351.81  4895.8  350.06  4911.8  349.76  4932.5  348.91
  4944.7  349.54  4984.2  347.87    4987  347.37  4990.2  347.87  5149.4  349.05
  5173.9  350.01  5188.1  349.28  5315.3  354.33  5513.3  365.18  5555.8  369.71
  5697.2  381.22  5711.3  381.33  5725.5  384.13  5753.8  387.06  5838.6  393.91
#Mann= 5 ,-1 , 0
    4587     .05       0  4911.8     .07       0  4984.2     .07       0
  4990.2     .07       0  5149.4     .05       0
Bank Sta=4864.1,5173.9
XS Rating Curve= 0 ,0
Exp/Cntr=0.3,0.1

Type RM Length L Ch R = 1 ,134321  ,494,494,494
BEGIN DESCRIPTION:
BIG ELKHART CREEK 168.0
END DESCRIPTION:
XS GIS Cut Line= 3
      3796349.57     10551360.22      3795999.61     10551710.19
      3795499.63     10552260.17
#Sta/Elev= 30
  4489.9  381.97  4503.9  381.91  4546.4  380.01  4560.6  377.33  4617.1  372.92
  4673.7  363.04  4716.1  358.89  4730.3   354.5  4758.6  350.13  4788.8  349.99
  4811.2  349.38  4928.3  349.39  4984.8  348.31  4995.7  346.81  4998.4  346.31
  5001.7  346.81  5012.9  348.06  5055.4  348.39  5091.3  349.99  5147.3  354.79
  5204.1  357.37  5246.7  360.16  5254.1  361.46    5417  371.14  5423.7  370.76
  5565.6  380.61  5607.5  385.14  5643.3  386.84  5678.5  390.58  5728.1  393.96
#Mann= 6 ,-1 , 0
  4489.9     .08       0  4503.9     .05       0  4788.8     .07       0
  4811.2     .05       0  4995.7     .03       0  5001.7     .05       0
Bank Sta=4984.8,5012.9
XS Rating Curve= 0 ,0
Exp/Cntr=0.3,0.1

Type RM Length L Ch R = 1 ,133827  ,371,371,371
BEGIN DESCRIPTION:
BIG ELKHART CREEK 167.0
END DESCRIPTION:
XS GIS Cut Line= 3
      3796144.74     10550721.23      3795616.95     10551474.72
      3795238.48     10552040.68
#Sta/Elev= 30
  4139.3  401.46  4299.6  389.14  4329.3  384.51    4365  382.25  4430.4  374.75
  4436.5  372.19  4501.9  363.15  4537.6  359.72  4558.6  359.25  4565.4  357.51
  4609.1  355.59  4615.2  354.01  4623.9  356.05    4630  353.98    4651  355.34
  4710.2  353.56  4716.3  352.42  4737.3  353.56  4945.6  348.55  4975.3  349.26
  4990.1  347.61  4993.2  345.46  4995.9  344.96  4999.2  345.46  5040.7  347.63
  5053.4  349.77  5211.8  358.93  5283.9  365.26    5479  378.17  5740.1  389.72
#Mann= 3 ,-1 , 0
  4139.3     .05       0  4993.2     .03       0  4999.2     .05       0
Bank Sta=4990.1,5053.4
XS Rating Curve= 0 ,0
Exp/Cntr=0.3,0.1

Type RM Length L Ch R = 1 ,133456  ,513,513,513
BEGIN DESCRIPTION:
BIG ELKHART CREEK 166.0
END DESCRIPTION:
XS GIS Cut Line= 3
      3795799.58     10550760.22      3795299.61     10551360.19
      3795199.61     10551760.19
#Sta/Elev= 30
  4250.9  390.73  4321.8  383.59  4364.8  380.44  4399.9  376.18  4435.1  374.05
  4471.5  369.85    4478  367.98  4492.3  367.36    4521  363.54  4527.5  361.49
  4556.1  357.73  4563.3  357.83  4591.3  353.22  4790.4  347.39  4797.6  348.07
  4833.4  346.83  4981.8  346.68  5000.9  345.73  5003.6  345.23  5006.9  345.73
  5018.2  346.87  5034.5  347.29  5049.9  349.47  5055.1  348.89  5091.2  352.03
  5114.3  355.37  5165.9  355.96  5214.8  361.51  5297.3  367.19  5444.2  379.69
#Mann= 3 ,-1 , 0
  4250.9     .05       0  5000.9     .03       0  5006.9     .05       0
Bank Sta=4981.8,5018.2
XS Rating Curve= 0 ,0
Exp/Cntr=0.3,0.1

Type RM Length L Ch R = 1 ,132943  ,520,520,520
BEGIN DESCRIPTION:
BIG ELKHART CREEK 165.0
END DESCRIPTION:
XS GIS Cut Line= 3
      3795049.62     10550660.15      3794949.61     10551110.19
      3794699.61     10551510.18
#Sta/Elev= 30
  4562.4  385.03  4623.9  379.75  4644.4  376.14    4679  373.44  4722.5  366.92
  4757.1  364.84    4766  362.82  4771.2  363.23  4814.7  357.24  4819.8   358.1
  4849.3  356.21  4906.9  348.02  4941.5  346.26  5001.2  344.46    5004  343.96
  5007.2  344.46  5028.6  345.13  5088.9  344.77 5104.27   346.9  5140.7  344.78
    5162  345.84  5177.2   345.2  5204.4  345.82  5256.3  349.96  5393.1  363.93
  5408.4  364.45  5429.7  368.12    5445  368.67  5450.9  370.45  5495.1   373.9
#Mann= 5 ,-1 , 0
  4562.4     .16       0  5001.2     .07       0  5007.2     .16       0
  5028.6     .12       0  5177.2     .16       0
Bank Sta=4941.5,5104.27
XS Rating Curve= 0 ,0
Exp/Cntr=0.3,0.1

Type RM Length L Ch R = 1 ,132423  ,470,470,470
BEGIN DESCRIPTION:
BIG ELKHART CREEK 164.0
END DESCRIPTION:
XS GIS Cut Line= 3
      3794749.59     10550710.22      3794549.61     10551060.19
      3794649.62     10551510.23
#Sta/Elev= 30
  4590.6   375.2  4598.5  375.36  4648.2  368.81  4694.2  365.16  4706.5  362.05
  4722.3  359.91  4728.8  357.42  4809.4  347.67  4818.8  347.79  4832.4  344.84
  4962.2  343.33  4996.2   343.7  5000.9  342.62  5003.7  342.12  5006.9  342.62
  5012.9  343.77  5034.7  343.16  5066.2  344.58  5105.1  343.21  5137.1  343.49
  5158.9  344.99  5167.5  347.27  5239.5  355.64  5245.9  357.26  5251.1  356.45
    5260  358.49  5289.5  361.58  5343.3  365.37  5403.4   372.5  5454.7   376.8
#Mann= 6 ,-1 , 0
  4590.6     .16       0  4962.2     .07       0  5000.9     .07       0
  5006.9     .07       0  5066.2     .12       0  5167.5     .16       0
Bank Sta=4996.2,5012.9
XS Rating Curve= 0 ,0
Exp/Cntr=0.3,0.1

Type RM Length L Ch R = 1 ,131953  ,336,336,336
BEGIN DESCRIPTION:
BIG ELKHART CREEK 163.0
END DESCRIPTION:
XS GIS Cut Line= 4
      3794349.62     10550310.15      3794149.61     10550910.19
      3793749.61     10551260.19      3793495.39     10551440.03
#Sta/Elev= 30
  4346.1   392.6  4388.3  388.01  4409.4  383.45  4419.9  378.87    4441  374.94
  4483.2  370.42  4493.7  366.71  4525.3   363.5  4546.4  357.03  4599.1  347.05
  4783.4   344.3  4936.4   343.6  5003.6  341.58  5006.3  341.08  5009.6  341.58
  5049.3  342.72  5056.9   345.1    5075  346.94  5093.2  348.35    5190  354.24
  5368.2  368.93  5417.6  370.82  5453.6  375.41  5460.3  380.33  5506.8  384.83
  5582.7  388.73  5718.3  399.32  5761.2   399.8  5796.9  405.13  5821.5  405.32
#Mann= 7 ,-1 , 0
  4346.1     .16       0  4783.4     .12       0  5003.6     .07       0
  5009.6     .12       0    5075     .16       0  5093.2     .12       0
    5190     .16       0
Bank Sta=4936.4,5056.9
XS Rating Curve= 0 ,0
Exp/Cntr=0.3,0.1

Type RM Length L Ch R = 1 ,131617  ,506,506,506
BEGIN DESCRIPTION:
BIG ELKHART CREEK 162.0
END DESCRIPTION:
XS GIS Cut Line= 3
      3794249.61     10550160.18      3794044.33     10550595.54
      3793449.62     10551110.18
#Sta/Elev= 30
    4477  405.23  4610.6  388.41    4665  373.35  4709.2  367.12  4731.3  356.74
  4747.3  353.31  4775.6  343.38  4786.6  342.89  4818.1  341.47  4820.9  340.97
  4824.1  341.47  4875.7  341.94  4878.9  341.99    4996  341.67  5078.5  342.93
  5099.4  341.65  5149.7  344.31  5184.5  344.14  5361.5  357.69    5447   360.9
  5475.5  359.31  5567.7  362.05  5574.3   364.5  5596.2  364.17  5645.6   370.7
  5688.3  372.05  5723.4     379  5731.1  378.06  5737.7  380.76  5744.8  380.05
#Mann= 7 ,-1 , 0
    4477     .16       0  4818.1     .07       0  4824.1     .16       0
  4875.7     .12       0  4878.9     .16       0    4996     .12       0
  5184.5     .16       0
Bank Sta=4786.6,5149.7
XS Rating Curve= 0 ,0
Exp/Cntr=0.3,0.1

Type RM Length L Ch R = 1 ,131111  ,470,470,470
BEGIN DESCRIPTION:
BIG ELKHART CREEK 161.0
END DESCRIPTION:
XS GIS Cut Line= 3
      3793999.62     10550110.17      3793799.61     10550360.19
      3793199.61     10550660.19
#Sta/Elev= 30
  4699.2  390.38  4720.8  386.64  4735.2  381.26  4756.1  377.97  4784.9  376.38
  4827.3  371.02  4848.9  368.08  4898.5   357.8  4919.3  355.95  4933.7  352.57
  4941.7  348.09  4948.1     347  4955.3  342.98  4965.5  341.22  4983.4   341.6
  4994.8  339.04  4997.5  338.54  5000.8  339.04  5005.8  341.41  5145.2  342.62
    5229  345.79  5310.1  346.55  5354.8  347.97  5386.2  351.32  5452.6  362.16
  5497.3  367.29  5502.9  366.52  5564.4  372.24  5623.1  374.84  5690.2  380.66
#Mann= 5 ,-1 , 0
  4699.2     .16       0  4965.5     .12       0  4994.8     .07       0
  5000.8     .12       0  5386.2     .16       0
Bank Sta=4983.4,5005.8
XS Rating Curve= 0 ,0
Exp/Cntr=0.3,0.1

Type RM Length L Ch R = 1 ,130641  ,447,447,447
BEGIN DESCRIPTION:
BIG ELKHART CREEK 160.0
END DESCRIPTION:
XS GIS Cut Line= 3
      3793849.58      10549910.2      3793549.61     10550010.19
      3792949.61     10550460.19
#Sta/Elev= 30
  4665.3  389.85  4675.8  388.76  4686.4  384.53  4728.5  375.31  4876.8  356.11
  4897.2  354.33  4907.7   350.4    4971  340.04  4984.6  339.37  5000.4  337.94
  5003.1  337.44  5006.4  337.94    5018  341.63  5109.6  339.38  5224.2  342.22
    5268  348.05  5274.2  347.01  5288.8  352.48    5297  351.96  5303.4  354.45
  5324.2  355.97  5331.5  359.83  5353.4  364.32    5445  368.66    5595  380.04
  5631.5  381.86  5638.8  380.09    5645  381.88  5674.2  383.09  5731.5  389.49
#Mann= 5 ,-1 , 0
  4665.3     .16       0  4876.8     .12       0  5000.4     .07       0
  5006.4     .12       0    5297     .16       0
Bank Sta=4984.6,5018
XS Rating Curve= 0 ,0
Exp/Cntr=0.3,0.1

Type RM Length L Ch R = 1 ,130194  ,506,506,506
BEGIN DESCRIPTION:
BIG ELKHART CREEK 159.0
END DESCRIPTION:
XS GIS Cut Line= 2
      3793828.36      10549177.2      3792718.99     10550213.66
#Sta/Elev= 30
  4181.8  416.95  4395.4  408.54  4508.5   395.8  4558.1  387.57  4572.2  381.57
  4628.9  370.45  4643.1  365.18  4664.1  361.56  4671.4  358.45  4678.2  358.45
  4714.2  347.86  4734.9  341.88  4805.7   339.1  4989.4  340.19  4996.7  337.41
  5014.8  337.08  5017.5  336.58  5020.8  337.08  5025.1  341.25  5116.4  358.94
  5166.3  364.52  5301.1  367.31  5470.6  377.42  5492.1  376.93    5605  385.03
  5619.1  381.15  5640.6  385.18  5661.6  386.31  5675.8  390.96    5700  392.04
#Mann= 5 ,-1 , 0
  4181.8     .16       0  4714.2     .12       0  5014.8     .07       0
  5020.8     .12       0  5116.4     .16       0
Bank Sta=4989.4,5025.1
XS Rating Curve= 0 ,0
Exp/Cntr=0.3,0.1

Type RM Length L Ch R = 1 ,129688  ,215,215,215
BEGIN DESCRIPTION:
BIG ELKHART CREEK 158.0
END DESCRIPTION:
XS GIS Cut Line= 2
      3793276.29     10548849.04      3792594.31     10550051.62
#Sta/Elev= 30
  4354.6  413.76    4419   409.9  4434.9  406.19  4521.4  396.26    4543   392.2
  4574.3  382.74  4623.8  371.14  4631.8  366.77    4683  350.77  4689.3  346.48
  4704.6  343.59  4712.3  340.17  4726.2  337.46  4755.3  337.78  4976.7  339.03
  4984.4  336.54  4996.7  335.72  4999.4  335.22  5002.7  335.72  5006.1  337.57
  5027.7  339.64  5034.2  342.23  5086.9  352.43    5110  354.84    5146  360.46
  5195.1  364.86  5496.5  373.98  5620.5  379.84  5658.1   384.2  5737.1   387.5
#Mann= 5 ,-1 , 0
  4354.6     .16       0  4755.3     .12       0  4996.7     .07       0
  5002.7     .12       0    5110     .16       0
Bank Sta=4976.7,5006.1
XS Rating Curve= 0 ,0
Exp/Cntr=0.3,0.1

Type RM Length L Ch R = 1 ,129473  ,472,472,472
BEGIN DESCRIPTION:
BIG ELKHART CREEK 157.0
END DESCRIPTION:
XS GIS Cut Line= 2
      3793229.41     10548781.36      3792317.95     10549854.27
#Sta/Elev= 30
  4369.8  415.25    4447  409.04  4552.8  395.81  4567.1  391.29  4581.4  389.39
  4595.7  383.31  4603.4  383.65    4610  379.96  4638.5  375.62  4673.6  364.16
  4709.4  358.03  4769.9  342.35  4794.5  336.76  4985.6  337.72  4990.3  334.82
    4993  334.32  4996.3  334.82  5014.1  335.34  5021.8  337.86  5074.5  343.34
  5149.2  350.68  5198.6  351.06  5212.9  353.65  5227.2  352.14  5319.5  354.96
  5362.3  362.46  5411.7  363.09  5489.7  367.22  5518.3  370.69  5777.6   381.7
#Mann= 5 ,-1 , 0
  4369.8     .16       0  4769.9     .12       0  4990.3     .07       0
  4996.3     .12       0  5074.5     .16       0
Bank Sta=4985.6,5021.8
XS Rating Curve= 0 ,0
Exp/Cntr=0.3,0.1

Type RM Length L Ch R = 1 ,129001  ,619,619,619
BEGIN DESCRIPTION:
BIG ELKHART CREEK 156.0
END DESCRIPTION:
XS GIS Cut Line= 2
      3793146.06     10548578.25      3791803.77     10549384.66
#Sta/Elev= 30
  4411.8  404.59  4425.2  401.88  4446.6  402.53  4504.9  396.35  4557.3  385.44
  4621.5  380.79  4695.3  368.83  4759.4  364.91  4790.5  359.09  4796.3  360.16
  4811.9  357.37  4833.3  356.86  4891.6  348.89  4907.2  344.42  4992.6   335.2
  4999.3  333.26  5002.1  332.76  5005.3  333.26  5023.7  337.33  5174.2  338.23
  5175.8  338.26  5329.3  339.97  5436.6  354.45  5480.9  362.99  5532.8  368.35
    5628  366.77  5707.6  374.38  5750.4  375.38  5802.8  373.04  5977.7  381.53
#Mann= 7 ,-1 , 0
  4411.8     .05       0  4907.2     .12       0  4999.3     .07       0
  5005.3     .12       0  5174.2     .16       0  5175.8     .12       0
  5436.6     .16       0
Bank Sta=4992.6,5023.7
XS Rating Curve= 0 ,0
Exp/Cntr=0.3,0.1

Type RM Length L Ch R = 1 ,128382  ,867,867,867
BEGIN DESCRIPTION:
BIG ELKHART CREEK 155.0
END DESCRIPTION:
XS GIS Cut Line= 3
      3793276.24     10548208.47      3791687.73     10548802.21
      3791406.46     10549203.27
#Sta/Elev= 30
  4041.4  406.49  4197.9  392.63  4233.6  391.93  4313.8  381.65  4336.7  382.54
  4374.4  377.25  4379.8  379.43  4390.1  375.74  4539.6  367.08    4605  360.35
  4731.7  353.15  4807.5  344.17  4909.9  337.66  4978.6  336.23  5000.5  331.02
  5003.3  330.52  5006.5  331.02  5009.3  335.36  5064.1  337.63  5290.5  334.87
  5297.5  332.46  5406.3  339.07  5469.1  347.72  5516.8  359.92  5577.4  363.58
  5671.2  375.06  5884.7  377.84  5950.1  375.05  6128.8  381.74  6227.1  391.52
#Mann= 6 ,-1 , 0
  4041.4     .05       0    4605     .16       0  4909.9     .12       0
  5000.5     .07       0  5006.5     .12       0  5469.1     .16       0
Bank Sta=4978.6,5009.3
XS Rating Curve= 0 ,0
Exp/Cntr=0.3,0.1
