HEC-RAS study BIG ELKHART CREEK.prj: BIG ELKHART CREEK Base Level Engineering

--- BIG ELKHART CREEK.g01 (geometry) --- (continued)

Type RM Length L Ch R = 1 ,127515  ,364,364,364
BEGIN DESCRIPTION:
BIG ELKHART CREEK 154.0
END DESCRIPTION:
XS GIS Cut Line= 4
      3792497.15     10547525.08      3791908.61     10548092.78
      3791575.28     10548457.36      3791294.34     10548634.25
#Sta/Elev= 30
  4027.1   415.2  4142.1  414.17  4255.3  402.82  4297.8  396.54    4333  388.11
  4389.6  382.02    4411  377.29  4417.9  372.46  4439.3  366.33  4446.2  362.35
  4453.4  361.65  4460.4  357.06  4531.1  340.46  4538.1  337.23  4559.4  335.92
  4566.4  333.62  4604.7  332.41  4976.8  332.97  4983.9  329.95  5001.8  329.21
  5004.6  328.71  5007.8  329.21  5012.2   332.5  5115.2  345.26  5139.4  348.82
  5189.2  360.19  5217.6   363.5  5431.4  372.36    5511  377.72  5670.8  378.16
#Mann= 5 ,-1 , 0
  4027.1     .16       0  4604.7     .12       0  5001.8     .07       0
  5007.8     .12       0  5115.2     .16       0
Bank Sta=4976.8,5012.2
XS Rating Curve= 0 ,0
Exp/Cntr=0.3,0.1

Type RM Length L Ch R = 1 ,127151  ,378,378,378
BEGIN DESCRIPTION:
BIG ELKHART CREEK 153.0
END DESCRIPTION:
XS GIS Cut Line= 3
      3792340.88     10547389.67      3791637.78     10547806.32
      3791330.49     10548410.48
#Sta/Elev= 30
  4021.3  416.03  4162.3   399.7  4190.2  394.88  4197.1  389.48  4211.6  387.67
  4227.2  381.04  4264.3  378.87  4270.1  374.53  4285.7  376.82  4291.5  371.75
  4301.3  374.42  4328.6  372.76  4344.2  374.66    4350  371.77  4371.5  369.47
  4424.1  371.96  4519.7  366.48  4546.9  355.46  4627.2  338.11  4662.2  334.51
  4743.8  329.67  4988.8  331.55  4994.2  328.94  4996.9  328.44  5000.2  328.94
  5011.2  332.31  5063.9  333.67  5135.1  341.12  5325.3  362.95  5516.4  375.85
#Mann= 5 ,-1 , 0
  4021.3     .16       0  4662.2     .12       0  4994.2     .07       0
  5000.2     .12       0  5135.1     .16       0
Bank Sta=4988.8,5011.2
XS Rating Curve= 0 ,0
Exp/Cntr=0.3,0.1

Type RM Length L Ch R = 1 ,126773  ,257,257,257
BEGIN DESCRIPTION:
BIG ELKHART CREEK 152.0
END DESCRIPTION:
XS GIS Cut Line= 3
      3791999.59      10547310.2      3791399.61     10547660.19
      3791249.58     10547910.23
#Sta/Elev= 30
  4336.1  397.82    4339  397.82  4343.9  394.79  4365.4  390.71  4408.4  388.56
  4439.9  384.29  4445.6  384.91  4461.4   380.4  4510.1  375.55  4568.9   367.1
  4584.6  366.29  4590.8  364.42  4621.8  361.24    4702  356.55  4723.5   353.3
  4739.2  353.31  4745.5  346.74  4810.7  338.01  4819.4  335.57  4825.2  336.94
  4899.6  329.31  4985.6  330.77  4998.3  327.98  5001.1  327.48  5004.3  327.98
  5017.1  330.18  5176.5  332.48  5205.6  335.38  5269.1     346  5322.3  353.71
#Mann= 5 ,-1 , 0
  4336.1     .16       0  4745.5     .12       0  4998.3     .07       0
  5004.3     .12       0  5269.1     .16       0
Bank Sta=4985.6,5017.1
XS Rating Curve= 0 ,0
Exp/Cntr=0.3,0.1

Type RM Length L Ch R = 1 ,126516  ,184,184,184
BEGIN DESCRIPTION:
Mapping XS e460eb6f
END DESCRIPTION:
XS GIS Cut Line= 3
      3792088.74     10547213.67      3791203.35     10547494.91
      3790470.71     10547785.89
#Sta/Elev= 30
    4151  412.89  4202.6  407.41    4276  391.24  4354.4  385.12  4380.9  381.16
  4386.7  378.03  4391.9  379.44    4419  375.44  4424.2  376.64  4451.2  371.23
  4464.9  372.19  4515.7  362.03    4650  352.62  4769.1   335.9  4790.9  335.23
    4881  330.81  4926.5  330.95    4997  327.18  4999.7  326.68    5003  327.18
    5010  330.58  5268.3  333.58  5376.3  338.57    5517  352.37  5535.9  356.06
  5600.7  360.74  5649.3  367.74  5708.7  370.83  5757.3  376.96  5868.3  382.69
#Mann= 6 ,-1 , 0
    4151     .16       0  4790.9     .12       0    4997     .07       0
    5003     .12       0  5268.3     .16       0  5376.3     .05       0
Bank Sta=4926.5,5010
XS Rating Curve= 0 ,0
Exp/Cntr=0.3,0.1

Type RM Length L Ch R = 1 ,126332  ,97,97,97
BEGIN DESCRIPTION:
Mapping XS 2734fadb
END DESCRIPTION:
XS GIS Cut Line= 3
      3792146.09     10546948.03      3791073.15     10547375.12
      3790375.22     10547599.08
#Sta/Elev= 30
  3927.9  404.18  4043.1   390.5  4096.2  385.94  4218.9  373.79  4259.2  366.72
  4338.2  358.25  4351.1  354.24  4356.4   356.4    4405  350.42  4620.8  337.73
  4626.2  339.78  4645.1  336.77  4860.5  334.19  4890.5  333.08  4895.9  329.65
  4914.3  332.65  4925.6  329.48  4944.5  331.82  4957.4  329.07  4974.1     332
  5000.8   327.1  5003.5   326.6  5006.8   327.1  5011.2  329.46  5043.5  328.92
  5057.7  332.65  5210.5  334.12  5306.9     339    5580  372.63  5815.7  387.24
#Mann= 7 ,-1 , 0
  3927.9     .05       0  4043.1      .1       0  4096.2     .05       0
  4259.2      .1       0  4338.2     .05       0  5000.8     .04       0
  5006.8     .05       0
Bank Sta=4974.1,5057.7
XS Rating Curve= 0 ,0
Exp/Cntr=0.3,0.1

Type RM Length L Ch R = 1 ,126235  ,520,520,520
BEGIN DESCRIPTION:
BIG ELKHART CREEK 151.0
END DESCRIPTION:
XS GIS Cut Line= 3
      3791349.61     10546510.19      3791099.61     10547310.19
      3790599.58      10547460.2
#Sta/Elev= 30
  4118.9  401.52  4160.8  396.99  4276.1  378.27    4318  372.82  4328.4  372.67
  4405.4  361.86  4412.3  359.23  4502.9  342.02  4548.5  340.43  4590.4  336.38
  4605.6  333.72    4699  331.16  4946.6  331.84  4973.6  330.52  4988.4  326.93
  5003.6  326.69  5006.4  326.19  5009.6  326.69  5011.9  329.17  5022.1  329.58
  5044.9   332.6    5078  331.69  5137.3  332.93  5182.4  333.51  5259.8  339.63
  5301.6  344.38  5332.9  352.49  5364.2  355.43  5396.4  361.56  5479.1  370.34
#Mann= 6 ,-1 , 0
  4118.9     .16       0    4699     .12       0  5003.6     .07       0
  5009.6     .12       0  5022.1      .1       0  5137.3     .05       0
Bank Sta=4973.6,5011.9
XS Rating Curve= 0 ,0
Exp/Cntr=0.3,0.1

Type RM Length L Ch R = 1 ,125715  ,530,530,530
BEGIN DESCRIPTION:
BIG ELKHART CREEK 150.0
END DESCRIPTION:
XS GIS Cut Line= 3
      3791249.58     10546360.23      3790749.61     10547010.19
      3790499.62     10547360.17
#Sta/Elev= 30
  4200.6  409.32  4301.2  396.39  4357.3  382.92    4457  370.14  4500.5  361.43
  4521.3   361.3  4535.8  355.68  4550.3  355.76  4571.2  352.82  4585.7  353.52
  4606.5  349.65  4714.3  337.11  4720.7  338.11  4728.9  335.04  4814.1  328.37
  4992.5  329.99    5004  325.97  5006.8  325.47    5010  325.97  5013.4  328.56
  5030.4  329.51  5128.8  329.14  5164.4  331.36  5185.3  333.95  5220.9  342.06
  5229.5  341.99  5250.4  347.41  5271.3  348.91  5315.5  358.11  5450.7  373.72
#Mann= 5 ,-1 , 0
  4200.6     .16       0  4814.1     .12       0    5004     .07       0
    5010     .12       0  5030.4     .05       0
Bank Sta=4992.5,5013.4
XS Rating Curve= 0 ,0
Exp/Cntr=0.3,0.1

Type RM Length L Ch R = 1 ,125185  ,553,553,553
BEGIN DESCRIPTION:
BIG ELKHART CREEK 149.0
END DESCRIPTION:
XS GIS Cut Line= 3
      3791199.63     10546310.18      3790649.61     10546560.19
      3790149.61     10547260.18
#Sta/Elev= 30
  4414.5  407.78  4513.4  394.62  4567.2  383.19  4624.3  374.25  4722.1  361.44
  4739.7  362.19    4777  357.86  4831.9  348.57  4903.9  332.27  4941.8  328.27
  4994.5  328.48  4996.7  328.35  5006.9  324.77  5009.6  324.27  5012.9  324.77
  5015.9  327.05  5026.3  328.77  5101.6  326.89  5276.7  327.67    5305  334.16
  5340.6  329.73  5435.3  331.23  5470.9  334.02  5511.8  342.76  5600.4  353.38
  5649.1  357.65  5657.7  360.45  5693.3  363.77  5806.4  381.25  5878.9  383.69
#Mann= 9 ,-1 , 0
  4414.5     .16       0  4903.9     .12       0  4994.5     .16       0
  5006.9     .07       0  5012.9     .16       0  5026.3     .12       0
  5101.6     .05       0  5511.8      .1       0  5600.4     .05       0
Bank Sta=4996.7,5015.9
XS Rating Curve= 0 ,0
Exp/Cntr=0.3,0.1

Type RM Length L Ch R = 1 ,124632  ,562,562,562
BEGIN DESCRIPTION:
BIG ELKHART CREEK 148.0
END DESCRIPTION:
XS GIS Cut Line= 3
      3791099.65     10546110.19      3790549.61     10546060.19
      3789799.65     10546160.18
#Sta/Elev= 30
  4413.5  396.96  4483.8  387.34    4534  378.93  4654.5  365.58  4704.7  354.03
  4734.9  349.34    4765  342.75  4795.1  338.92    4825  336.84  4855.4  332.21
  4895.5  328.56  4945.7   326.4  4978.1  327.92 4996.23  326.77  4999.4  324.02
  5002.1  323.52  5005.4  324.02  5007.4  326.18  5026.3   328.2  5066.7  326.13
  5123.9  326.08  5288.6  328.77  5467.8  329.91  5500.5  332.23  5520.7  336.95
  5607.7  350.87  5612.7  350.22  5641.7  354.76  5694.6  359.53  5722.4  361.24
#Mann= 8 ,-1 , 0
  4413.5     .16       0    4825     .12       0  4978.1     .16       0
  4999.4     .07       0  5005.4     .16       0  5123.9     .05       0
  5467.8     .16       0  5694.6     .05       0
Bank Sta=4996.23,5007.4
XS Rating Curve= 0 ,0
Exp/Cntr=0.3,0.1

Type RM Length L Ch R = 1 ,124070  ,541,541,541
BEGIN DESCRIPTION:
BIG ELKHART CREEK 147.0
END DESCRIPTION:
XS GIS Cut Line= 3
      3790899.57     10545610.18      3790349.61     10545560.19
      3789899.58      10545710.2
#Sta/Elev= 30
  4460.3  385.49  4510.5  380.21  4550.6  373.07  4560.7  372.39  4610.9  364.68
    4641  362.47  4661.1  357.82  4691.2  354.77  4701.2  352.57  4781.6  341.04
  4801.7  339.41  4821.7  335.44  4831.8   334.5  4850.4  329.67  4932.2  325.56
  4982.4  326.12  4999.5  323.22  5002.2  322.72  5005.5  323.22  5015.2  323.31
  5023.1  326.38    5169  324.96  5212.8  324.82    5255  326.28  5265.5   328.3
  5297.1  331.15  5307.7  333.65  5370.9     343  5429.1   348.4  5486.9  352.29
#Mann= 6 ,-1 , 0
  4460.3     .16       0  4850.4     .12       0  4999.5     .07       0
  5005.5     .12       0    5169     .16       0  5429.1     .05       0
Bank Sta=4982.4,5023.1
XS Rating Curve= 0 ,0
Exp/Cntr=0.3,0.1

Type RM Length L Ch R = 1 ,123529  ,561,561,561
BEGIN DESCRIPTION:
BIG ELKHART CREEK 146.0
END DESCRIPTION:
XS GIS Cut Line= 3
      3790499.62     10544760.18      3790199.61     10545060.19
      3789849.59     10545510.22
#Sta/Elev= 30
  4540.9  407.72  4668.2  391.82  4710.6  385.15  4738.9  378.78    4753   372.7
  4837.9  361.12  4894.5  348.83    4951  332.42  4961.6  327.44  4968.3  327.44
  4972.4  325.43  4986.9   324.7  4990.2  322.48    4993  321.98  4996.2  322.48
  4997.9  322.51  5001.4  322.58  5007.7  324.87  5100.9  324.54  5115.4  323.18
  5150.7  324.96    5186  323.41  5200.5  325.16  5235.7  324.05  5264.7  328.84
  5307.2  332.25  5328.9  336.76  5396.9  343.14  5457.4  346.92  5535.3   349.4
#Mann= 5 ,-1 , 0
  4540.9     .16       0  4990.2     .07       0  4996.2     .16       0
  4997.9     .12       0  5396.9     .16       0
Bank Sta=4986.9,5007.7
XS Rating Curve= 0 ,0
Exp/Cntr=0.3,0.1

Type RM Length L Ch R = 1 ,122968  ,683,683,683
BEGIN DESCRIPTION:
BIG ELKHART CREEK 145.0
END DESCRIPTION:
XS GIS Cut Line= 3
      3790399.61     10544560.19      3789799.61     10544760.19
      3789399.58      10544960.2
#Sta/Elev= 30
  4344.5  407.99  4439.4  394.63  4449.9  394.56  4523.7  380.56  4597.5  373.25
  4618.6  369.05  4629.1  365.33  4671.3  358.29  4713.4  352.42  4734.5  351.69
  4745.1  348.78  4766.1  347.43  4776.7  342.76  4850.5  327.47  4855.3  327.05
  4892.6  323.47  4979.8  324.14  4999.3  322.52  5021.7  323.18    5041  321.03
  5043.8  320.53    5047  321.03  5088.8  323.07  5192.2  323.51  5236.9  327.54
    5276  333.05  5281.6  332.48    5290  335.02    5384  349.99  5424.2  354.13
#Mann= 5 ,-1 , 0
  4344.5     .16       0  4855.3     .12       0    5041     .07       0
    5047     .12       0    5384     .16       0
Bank Sta=4850.5,5236.9
XS Rating Curve= 0 ,0
Exp/Cntr=0.3,0.1

Type RM Length L Ch R = 1 ,122285  ,565,565,565
BEGIN DESCRIPTION:
BIG ELKHART CREEK 144.0
END DESCRIPTION:
XS GIS Cut Line= 3
      3790149.64     10544260.19      3789749.61     10544210.19
      3789199.65     10544210.19
#Sta/Elev= 30
    4622  379.04  4652.3  372.76  4659.8  369.88  4745.5  361.58    4753  358.71
  4783.3  355.78  4803.4  351.95  4826.1  346.89  4833.7  342.53  4864.2  340.87
  4884.1  338.85  4924.4  327.26  4934.4  326.51  4944.5  324.05  4974.8  322.47
  4979.3  319.88  4982.1  319.38  4985.3  319.88  4987.4  321.61    5005  320.56
  5035.1  323.46  5095.1  323.86  5155.1  321.91    5265  322.84  5335.1  323.29
  5375.1  325.25  5445.1  337.02  5475.1  340.54  5515.1  348.93  5575.1  354.72
#Mann= 5 ,-1 , 0
    4622     .16       0  4864.2     .12       0  4979.3     .07       0
  4985.3     .12       0    5265     .05       0
Bank Sta=4934.4,5035.1
XS Rating Curve= 0 ,0
Exp/Cntr=0.3,0.1

Type RM Length L Ch R = 1 ,121720  ,512,512,512
BEGIN DESCRIPTION:
BIG ELKHART CREEK 143.0
END DESCRIPTION:
XS GIS Cut Line= 3
      3790099.65     10543560.17      3789599.61     10543760.19
      3789299.62     10544060.17
#Sta/Elev= 30
  4452.1   391.8  4491.2  384.05  4496.6  384.93    4506  380.85  4520.8     379
    4545  368.74  4550.4  369.71  4598.9  357.67  4613.7  358.02  4652.7  350.25
    4677  350.47  4682.4  348.87  4689.1  351.32  4706.6  352.73  4730.8   352.1
  4742.9  347.07  4796.8  334.54  4814.3  333.57  4819.7  330.46  4915.3  319.58
  4949.1   321.3  4981.2  321.95    4985  318.92  4987.7  318.42    4991  318.92
  5033.1  321.91  5204.1  320.55  5231.1  321.83  5344.2   339.1  5414.9  346.42
#Mann= 5 ,-1 , 0
  4452.1     .16       0  4949.1     .12       0    4985     .07       0
    4991     .12       0  5204.1     .05       0
Bank Sta=4981.2,5033.1
XS Rating Curve= 0 ,0
Exp/Cntr=0.3,0.1

Type RM Length L Ch R = 1 ,121208  ,492,492,492
BEGIN DESCRIPTION:
BIG ELKHART CREEK 142.0
END DESCRIPTION:
XS GIS Cut Line= 3
      3789999.56     10543410.19      3789399.61     10543410.19
      3789049.59     10543660.21
#Sta/Elev= 30
  4410.8  385.59  4450.8  379.97  4480.8  372.96  4520.8  366.56  4550.8  363.86
  4580.8  359.02  4700.8   344.9  4710.8  342.14  4770.8  333.13  4840.8  326.68
  4850.8  324.92  4920.8  320.27  4980.8  320.94  4991.4  317.75  4997.8  317.23
  5000.5  316.73  5003.8  317.23  5013.8  318.17  5018.1  320.72    5125  318.49
  5169.3  318.98  5190.2  319.69  5204.9  321.44  5211.1  320.89  5246.7   326.9
  5261.5  327.61  5276.2  329.94  5297.1  334.91  5384.7  342.47  5440.9   346.1
#Mann= 5 ,-1 , 0
  4410.8     .16       0  4991.4     .12       0  4997.8     .07       0
  5003.8     .12       0  5384.7     .05       0
Bank Sta=4980.8,5018.1
XS Rating Curve= 0 ,0
Exp/Cntr=0.3,0.1

Type RM Length L Ch R = 1 ,120716  ,128,128,128
BEGIN DESCRIPTION:
BIG ELKHART CREEK 141.0
END DESCRIPTION:
XS GIS Cut Line= 3
      3789227.57     10542244.75      3789251.88     10542897.52
      3788949.92     10543775.63
#Sta/Elev= 30
  4256.1   347.2  4271.6  345.17  4381.6  341.99  4463.8   332.8  4491.7  330.18
  4511.7  326.25  4531.7  324.28  4611.8  319.13  4781.9  318.28    4852  319.35
    4862  318.04    4869  315.59  4871.7  315.09    4875  315.59    4882  319.53
  4913.4  318.26  4975.6  319.62  4986.2  319.51  4992.3  315.96  5017.9  319.81
    5039  318.44  5292.8  318.03  5419.1  320.57  5455.6  324.19  5486.4  328.97
  5493.8  330.91  5504.3  330.87  5525.5   335.3  5684.1  347.31  5837.9  352.73
#Mann= 5 ,-1 , 0
  4256.1     .16       0  4463.8     .12       0    4869     .07       0
    4875     .12       0  5486.4     .05       0
Bank Sta=4975.6,5017.9
XS Rating Curve= 0 ,0
Exp/Cntr=0.3,0.1

Type RM Length L Ch R = 1 ,120588  ,507,507,507
BEGIN DESCRIPTION:
Mapping XS 2e7121dc
END DESCRIPTION:
XS GIS Cut Line= 3
      3789109.52     10542216.94      3789106.05     10543102.38
      3788880.83     10543646.36
#Sta/Elev= 30
  4214.8  350.07    4338  346.15    4368  344.15    4388  342.32  4437.8  334.29
    4448  333.54  4478.1  327.64  4508.1  324.94  4518.1  322.68  4588.1  318.17
  4938.1  318.89  4945.1  316.12  4947.8  315.62  4951.1  316.12  4958.1  318.73
  4978.1  319.39  4998.1  316.91  5018.1   319.5  5038.1  318.02  5119.5  317.92
  5141.2  320.82  5162.8  319.18  5195.3  319.44  5292.7  323.18  5357.6  323.65
  5411.7  329.04  5420.9  331.92  5494.5  338.51  5606.6  345.63    5689  349.35
#Mann= 5 ,-1 , 0
  4214.8     .16       0  4437.8     .12       0  4945.1     .07       0
  4951.1     .12       0  5420.9     .05       0
Bank Sta=4978.1,5018.1
XS Rating Curve= 0 ,0
Exp/Cntr=0.3,0.1

Type RM Length L Ch R = 1 ,120081  ,550,550,550
BEGIN DESCRIPTION:
BIG ELKHART CREEK 140.0
END DESCRIPTION:
XS GIS Cut Line= 3
      3789049.61     10542260.19      3788749.61     10542760.19
      3788499.61     10543110.18
#Sta/Elev= 30
  4387.4  347.64  4410.7  347.83  4422.4  345.06  4432.1  344.78  4453.5  341.87
  4480.7  335.81  4496.2  334.48    4504  332.08  4527.3  327.45    4579  321.59
  4671.2  316.68  4861.6  316.29  4973.6   318.4  4977.9   316.3  4989.6  313.15
  4992.4  312.65  4995.6  313.15  5007.4  317.12  5049.1  320.66  5084.8  321.63
  5105.7  325.98  5120.4  327.26    5129  328.89  5142.5  329.46  5191.7  335.59
  5276.1  341.31  5286.3  340.82  5292.5  341.95  5314.6  342.95  5400.6  345.43
#Mann= 5 ,-1 , 0
  4387.4     .16       0    4579     .12       0  4989.6     .07       0
  4995.6     .12       0  5276.1     .05       0
Bank Sta=4973.6,5007.4
XS Rating Curve= 0 ,0
Exp/Cntr=0.3,0.1

Type RM Length L Ch R = 1 ,119531  ,548,548,548
BEGIN DESCRIPTION:
BIG ELKHART CREEK 139.0
END DESCRIPTION:
XS GIS Cut Line= 3
      3788849.59     10541760.21      3788449.61     10542360.19
      3788099.58     10542710.22
#Sta/Elev= 30
  4244.3  366.27  4323.9  360.99  4329.9  359.41  4338.9  359.95    4375  356.28
  4504.2  339.43  4525.2   338.5  4532.7  336.13  4561.3  331.85  4568.8   328.7
  4591.3  323.01  4617.6  319.41  4669.4  316.47  4762.6   314.9  4828.7  314.61
  4870.7  316.16  4993.7  316.89  5004.8   313.2  5007.6   312.7  5010.8   313.2
    5022  316.75  5135.1  317.91  5149.2  320.46  5163.4  321.29  5177.5  324.61
  5191.7   325.2  5210.9  327.95  5276.5  337.12  5304.8   339.3  5460.4  342.54
#Mann= 5 ,-1 , 0
  4244.3     .16       0  4617.6     .12       0  5004.8     .07       0
  5010.8     .12       0  5210.9     .05       0
Bank Sta=4993.7,5022
XS Rating Curve= 0 ,0
Exp/Cntr=0.3,0.1

Type RM Length L Ch R = 1 ,118983  ,750,750,750
BEGIN DESCRIPTION:
BIG ELKHART CREEK 138.0
END DESCRIPTION:
XS GIS Cut Line= 3
      3788937.41     10541487.26      3788124.89     10542023.73
       3787224.2     10542617.24
#Sta/Elev= 30
  4269.9  383.82  4387.1  378.07  4494.9  364.09  4501.5     360  4522.6  358.77
  4552.7  349.58  4594.8  350.94  4609.9  347.22  4630.9   348.3  4638.7  345.11
    4652   345.7  4661.1  342.09  4667.1  343.66  4682.1  338.77  4703.2   338.4
  4718.2  333.72  4769.4  327.34  4873.8  320.66 4985.79  316.09  4995.2  311.51
    4998  311.01  5001.2  311.51  5013.2  316.45  5151.7  314.98  5476.9  318.75
  5638.9  338.45  5789.5  341.53  5901.5     340  6009.9  343.07  6322.2  360.39
#Mann= 6 ,-1 , 0
  4269.9     .16       0  4873.8     .12       0  4995.2     .07       0
  5001.2     .12       0  5638.9     .16       0  5789.5     .05       0
Bank Sta=4985.79,5013.2
XS Rating Curve= 0 ,0
Exp/Cntr=0.3,0.1

Type RM Length L Ch R = 1 ,118233  ,311,311,311
BEGIN DESCRIPTION:
BIG ELKHART CREEK 137.0
END DESCRIPTION:
XS GIS Cut Line= 2
      3788624.36     10540778.87      3786999.64     10542535.51
#Sta/Elev= 30
  4090.6  424.45  4130.3  422.57  4208.1  420.46  4455.9  397.18  4505.2  385.61
  4555.1  381.09  4561.9   375.9  4618.6  363.39    4668  367.93  4696.3  366.24
  4703.7  360.84  4710.5  365.25  4724.7  364.96    4732  359.36  4738.8  362.45
  4767.2  354.82  4788.2  357.93  4830.7  349.55  4923.1  319.11  4979.2  314.52
  4990.4  310.09  4993.2  309.59  4996.4  310.09    5015  314.86  5031.7  314.86
  5495.8  313.26  5606.3  326.16  5672.7  335.58  5896.7  343.39  6483.4  363.41
#Mann= 7 ,-1 , 0
  4090.6     .05       0  4130.3     .16       0  4990.4     .07       0
  4996.4     .16       0  5031.7     .12       0  5606.3     .16       0
  5896.7     .05       0
Bank Sta=4979.2,5015
XS Rating Curve= 0 ,0
Exp/Cntr=0.3,0.1

Type RM Length L Ch R = 1 ,117922  ,691,691,691
BEGIN DESCRIPTION:
BIG ELKHART CREEK 136.0
END DESCRIPTION:
XS GIS Cut Line= 3
      3788229.07     10540742.45      3787624.89     10541549.77
      3786890.51     10542341.44
#Sta/Elev= 30
  4117.9  405.23  4137.9  400.69    4165  402.71  4252.5   395.6    4315   382.2
    4438  369.85  4452.3  364.77  4458.8  359.64  4479.7  355.42  4508.9  344.16
  4608.4  334.58  4629.7  329.31  4638.1  330.94  4644.3  328.14  4694.3  325.73
  4708.9  321.16  4729.8  322.54  4838.1  312.95  4940.3  313.49  4994.4   313.9
  4998.9  310.02  5001.6  309.52  5004.9  310.02  5023.6  313.58  5257.7  312.43
  5339.9  319.45  5420.4   331.3  5491.3  336.61  6059.2     353  6206.1   357.7
#Mann= 6 ,-1 , 0
  4117.9     .16       0  4940.3     .12       0  4998.9     .07       0
  5004.9     .12       0  5339.9     .16       0  6059.2     .05       0
Bank Sta=4994.4,5023.6
XS Rating Curve= 0 ,0
Exp/Cntr=0.3,0.1

Type RM Length L Ch R = 1 ,117231  ,653,653,653
BEGIN DESCRIPTION:
BIG ELKHART CREEK 135.0
END DESCRIPTION:
XS GIS Cut Line= 4
      3788051.95     10540679.98      3787510.31     10540784.14
      3787239.47     10541086.23      3786734.43     10542143.18
#Sta/Elev= 30
  4199.6  381.27    4426  376.52  4751.2  356.44  4791.3  350.05  4798.8  347.07
  4833.9  339.93  4840.6   336.6  4883.2  329.11  4890.7   326.2  4974.8   313.2
  4989.4  311.36  4993.9  308.93  4996.6  308.43  4999.9  308.93  5017.8  312.17
  5138.1  309.96  5399.8  313.98  5535.9  331.65  5544.5  331.23  5609.5  330.75
  5626.6  332.55  5632.2   331.1  5654.9  333.18  5683.1  332.61  5693.3   334.6
  5715.4  333.15  5759.8   337.6  5909.9  345.95  6158.7  349.36  6328.3  354.61
#Mann= 5 ,-1 , 0
  4199.6     .16       0  4974.8     .12       0  4993.9     .07       0
  4999.9     .12       0  5544.5     .16       0
Bank Sta=4989.4,5017.8
XS Rating Curve= 0 ,0
Exp/Cntr=0.3,0.1

Type RM Length L Ch R = 1 ,116578  ,554,554,554
BEGIN DESCRIPTION:
BIG ELKHART CREEK 134.0
END DESCRIPTION:
XS GIS Cut Line= 3
      3787299.63     10540010.16      3786849.61     10540660.19
      3786449.61     10540910.19
#Sta/Elev= 30
  4208.3  359.34  4230.6  357.79  4236.7  352.62  4244.8  351.43  4338.1  349.27
    4359  343.85  4373.9  343.78    4380  339.55  4409.7   335.9  4415.8  331.83
  4430.6  327.13  4466.5  319.13  4524.6  316.52  4784.3  313.37    4905  310.88
  4976.6   312.3  4991.5  309.18  4995.9  306.18  5003.6   306.1  5006.3   305.6
  5009.6   306.1  5021.9   306.7  5027.8  311.47  5304.9  309.36  5340.9  314.63
  5347.4  320.78  5374.6  328.32  5389.8   329.7  5420.5  336.99  5470.6  342.47
#Mann= 5 ,-1 , 0
  4208.3     .16       0  4784.3     .12       0  5003.6     .07       0
  5009.6     .12       0  5374.6     .16       0
Bank Sta=4976.6,5027.8
XS Rating Curve= 0 ,0
Exp/Cntr=0.3,0.1

Type RM Length L Ch R = 1 ,116024  ,525,525,525
BEGIN DESCRIPTION:
BIG ELKHART CREEK 133.0
END DESCRIPTION:
XS GIS Cut Line= 3
      3786999.63     10539510.16      3786549.61     10540310.19
      3786149.63     10540410.18
#Sta/Elev= 30
    4077   400.4  4180.3  388.93  4193.4  383.19  4237.7  371.27  4246.9  371.96
  4252.6  369.49  4290.2  366.91    4296  364.34  4306.2  365.62  4376.9  355.95
  4414.5   343.6  4421.2  338.93  4436.2  336.83  4444.2  331.75  4457.9  329.15
  4479.6  320.24  4501.6  316.22  4560.5   310.7  4640.7  308.64    4972  310.09
    4992  305.63    5010  305.18  5012.7  304.68    5016  305.18  5025.8   309.7
  5177.9  313.71  5214.7  317.54  5260.3  323.62  5355.7  330.81  5407.2  337.79
#Mann= 5 ,-1 , 0
    4077     .16       0  4640.7     .12       0    5010     .07       0
    5016     .12       0  5214.7     .16       0
Bank Sta=4972,5025.8
XS Rating Curve= 0 ,0
Exp/Cntr=0.3,0.1

Type RM Length L Ch R = 1 ,115499  ,556,556,556
BEGIN DESCRIPTION:
BIG ELKHART CREEK 132.0
END DESCRIPTION:
XS GIS Cut Line= 3
      3786699.58      10539660.2      3786299.61     10539860.19
       3785949.6      10540260.2
#Sta/Elev= 30
  4553.6   362.5  4589.9   360.1  4612.3  356.33  4620.7   351.5  4634.6   347.1
    4643  342.03    4657  338.22  4665.4  332.65  4679.3  328.97  4696.1  321.23
  4710.1  319.21  4724.1  315.01  4813.5  306.78  4861.6  307.29  4992.4  309.02
    4998  304.34  5004.9  304.34  5007.7  303.84  5010.9  304.34  5022.1  309.31
  5071.5  307.98  5227.1  309.57  5312.6  313.81  5338.9     317  5433.1  328.83
  5475.8  331.94  5504.3  336.92  5525.2  337.11    5529  339.41  5532.3  339.41
#Mann= 5 ,-1 , 0
  4553.6     .16       0  4861.6     .12       0  5004.9     .07       0
  5010.9     .12       0  5338.9     .16       0
Bank Sta=4992.4,5022.1
XS Rating Curve= 0 ,0
Exp/Cntr=0.3,0.1

Type RM Length L Ch R = 1 ,114943  ,492,492,492
BEGIN DESCRIPTION:
BIG ELKHART CREEK 131.0
END DESCRIPTION:
XS GIS Cut Line= 3
      3786449.58     10539410.19      3785949.61     10539510.19
      3785549.59     10539810.21
#Sta/Elev= 30
  4488.2  356.15  4549.4  349.79  4590.1   342.9  4651.3  329.37  4671.7  322.78
  4681.9  317.27  4702.3  312.97  4732.9  309.11  4757.7  308.57  4804.3  306.96
  4814.5  308.03  4967.5  307.25  4984.9  303.89  4987.6  303.39  4990.9  303.89
  5005.4  304.22  5011.6  307.28  5119.9  307.41  5219.9   310.5  5226.2  309.42
  5309.9  315.01  5334.5  319.07  5340.8  318.39  5361.6  321.26  5369.9   324.5
  5390.8  325.73  5419.9  332.52  5440.8  334.77  5448.1  337.87  5498.1  342.86
#Mann= 5 ,-1 , 0
  4488.2     .16       0  4757.7     .12       0  4984.9     .07       0
  4990.9     .12       0  5309.9     .16       0
Bank Sta=4967.5,5011.6
XS Rating Curve= 0 ,0
Exp/Cntr=0.3,0.1

Type RM Length L Ch R = 1 ,114451  ,943,943,943
BEGIN DESCRIPTION:
BIG ELKHART CREEK 130.0
END DESCRIPTION:
XS GIS Cut Line= 3
      3786349.61     10539010.19      3785699.61     10539110.19
      3785299.57     10539060.18
#Sta/Elev= 30
  4375.7  350.71  4409.9  348.14  4436.4  343.74  4466.8  340.54  4473.1  337.86
    4487   337.1  4536.3  326.61  4588.2  319.58  4618.5  313.61  4638.8  310.95
  4689.4  307.85  4709.6  305.17  4741.2  307.24  4780.4  306.13  4851.2  306.57
  4861.4  304.94  4867.7  306.14  4901.8  307.15  4972.6  307.96  4996.2  303.34
    4999  302.84  5002.2  303.34  5013.1  303.43  5023.2  307.65  5103.9  306.77
  5156.8  310.94  5214.8  318.18  5297.2   331.8  5325.6   335.5  5436.5  339.42
#Mann= 6 ,-1 , 0
  4375.7     .16       0  4689.4     .12       0  4996.2     .07       0
  5002.2     .12       0  5156.8     .16       0  5297.2     .05       0
Bank Sta=4972.6,5023.2
XS Rating Curve= 0 ,0
Exp/Cntr=0.3,0.1

Type RM Length L Ch R = 1 ,113508  ,273,273,273
BEGIN DESCRIPTION:
BIG ELKHART CREEK 129.0
END DESCRIPTION:
XS GIS Cut Line= 3
       3786679.9       10538140.      3785603.51     10538563.61
      3785020.15     10538994.18
#Sta/Elev= 30
  4146.4  407.59  4264.7  401.95  4419.4  389.94  4540.9  377.38  4600.5  366.88
  4619.5  361.75  4630.3  356.01  4649.3  354.06  4654.6  351.59    4679  350.36
  4716.3  337.52    4727  335.96  4733.2  330.46    4763   320.7  4787.4  316.75
  4792.8   313.9  4846.9  306.19  4919.8  304.28  4985.1  304.98  5006.5  301.41
  5009.2  300.91  5012.5  301.41  5017.2  303.95  5264.4  306.02  5302.6  313.24
  5457.5  326.84    5482  325.82  5525.1  331.13  5572.8   332.4  6028.2  349.86
#Mann= 7 ,-1 , 0
  4146.4     .05       0  4419.4     .16       0  4919.8     .12       0
  5006.5     .07       0  5012.5     .12       0  5457.5     .16       0
  5572.8     .05       0
Bank Sta=4985.1,5017.2
XS Rating Curve= 0 ,0
Exp/Cntr=0.3,0.1

Type RM Length L Ch R = 1 ,113235  ,477,477,477
BEGIN DESCRIPTION:
BIG ELKHART CREEK 128.0
END DESCRIPTION:
XS GIS Cut Line= 3
      3786617.44     10537987.21       3785992.4     10538049.72
      3784965.22     10538875.63
#Sta/Elev= 30
  4135.1  407.04  4317.3  396.85  4464.2  385.02  4618.8  371.68    4787  342.99
  4836.6  339.68  4857.4  336.34  4871.8  329.32  4886.2  325.34  4894.2  320.17
  4900.6  321.07  4929.4  311.48  4964.6  304.13  4985.6  304.42  4993.4  303.38
  4996.8  300.57  4999.6  300.07  5002.8  300.57  5014.2  301.04  5022.2  304.86
    5107  302.83  5255.8  304.95  5319.8   303.7  5356.6  311.37  5391.8  315.92
    5427  316.16  5441.4  320.85  5510.1     326  5626.6  332.33  6081.3  348.88
#Mann= 6 ,-1 , 0
  4135.1     .05       0  4464.2     .16       0  4985.6     .12       0
  4996.8     .07       0  5002.8     .12       0  5510.1     .05       0
Bank Sta=4993.4,5022.2
XS Rating Curve= 0 ,0
Exp/Cntr=0.3,0.1

Type RM Length L Ch R = 1 ,112758  ,565,565,565
BEGIN DESCRIPTION:
BIG ELKHART CREEK 127.0
END DESCRIPTION:
XS GIS Cut Line= 3
      3786652.14     10537827.49      3785659.07     10537855.27
      3784743.48     10538888.78
#Sta/Elev= 30
  3669.1  401.42  3811.7  394.07    3880  388.14  4141.8  369.77  4241.9  349.26
  4341.9  342.18  4411.9  340.76    4632  308.81  4743.6  307.75  4757.9  305.17
  4764.5  307.31  4772.1  304.92  4807.2   306.5  4814.7  304.17  4821.4  306.66
  4838.5  305.74  4984.5  304.14  4991.2  300.25  5002.4  299.96  5005.2  299.46
  5008.4  299.96    5013  303.65  5111.6  303.84  5211.2  316.02  5305.8  321.96
  5345.8  324.79  5487.2  328.11  5530.8  331.65  5735.6  343.32  6043.3  355.77
#Mann= 7 ,-1 , 0
  3669.1     .05       0    3880     .16       0  4838.5     .12       0
  5002.4     .07       0  5008.4     .12       0  5305.8     .16       0
  5530.8     .05       0
Bank Sta=4984.5,5013
XS Rating Curve= 0 ,0
Exp/Cntr=0.3,0.1

Type RM Length L Ch R = 1 ,112193  ,678,678,678
BEGIN DESCRIPTION:
BIG ELKHART CREEK 126.0
END DESCRIPTION:
XS GIS Cut Line= 3
      3785549.62     10537110.17      3785099.61     10537810.19
      3784849.61     10538160.18
#Sta/Elev= 30
  4206.3  378.49  4252.1  376.44  4313.6   370.5    4350  361.43  4365.2  360.02
  4380.4  353.61  4422.6  349.32  4467.9  340.63  4495.3  338.46  4531.6  333.21
  4539.2  331.48  4546.8  327.12  4567.9  323.52  4574.9  319.78  4604.2  312.63
  4610.5  309.34  4640.6  304.84  4753.2  302.78  4937.1  301.79  4988.6  303.15
  4991.6  298.96  4994.3  298.46  4997.6  298.96  5009.8  299.05  5015.7  302.91
  5210.5  301.93  5283.8  309.29  5324.8  315.74  5401.2  322.83  5468.6  328.13
#Mann= 7 ,-1 , 0
  4206.3     .05       0  4252.1     .16       0  4753.2     .12       0
  4991.6     .07       0  4997.6     .12       0  5283.8     .16       0
  5401.2     .05       0
Bank Sta=4988.6,5015.7
XS Rating Curve= 0 ,0
Exp/Cntr=0.3,0.1

Type RM Length L Ch R = 1 ,111515  ,185,185,185
BEGIN DESCRIPTION:
BIG ELKHART CREEK 125.0
END DESCRIPTION:
XS GIS Cut Line= 6
      3785478.47     10537174.72      3785020.18     10537209.44
      3784756.29     10537292.77      3784561.85     10537501.11
      3784547.96     10537688.61      3784332.68     10538702.48
#Sta/Elev= 30
  4156.4  372.93  4375.9  342.66  4429.2  340.51  4466.1  341.69  4539.7  337.69
  4596.5  334.37  4618.9  330.66  4669.3  315.81    4711  306.44  4784.4  302.01
  4850.3  301.58  4922.6  301.86  4980.6   300.9  4982.8  300.35  4998.6  298.09
  5001.4  297.59  5004.6  298.09  5015.8  301.01  5052.2   301.2  5058.3  299.31
  5072.5  301.89    5159  301.87  5233.5   303.9    5257     304  5337.2  316.28
  5377.1  319.35    5526  326.91  6001.2  344.05    6175  353.21  6402.2  356.18
#Mann= 12 ,-1 , 0
  4156.4     .16       0  4539.7     .05       0  4669.3     .12       0
  4850.3     .05       0  4922.6     .12       0  4982.8     .16       0
  4998.6     .07       0  5004.6     .16       0  5052.2     .12       0
    5159     .05       0  5233.5     .12       0  5377.1     .05       0
Bank Sta=4980.6,5015.8
XS Rating Curve= 0 ,0
Exp/Cntr=0.3,0.1

Type RM Length L Ch R = 1 ,111330  ,246,246,246
BEGIN DESCRIPTION:
Mapping XS 551e6f8d
END DESCRIPTION:
XS GIS Cut Line= 6
      3785513.21     10537063.61      3784978.51     10537056.66
      3784672.96     10537105.27      3784471.57     10537334.44
      3784200.74     10537771.94       3783270.2      10538001.1
#Sta/Elev= 30
  3940.6  379.37  3956.6  378.35  4024.2  373.22  4084.2  366.05  4164.2   351.8
  4450.8  320.06    4592  307.81  4924.9  303.99  4967.5  302.67  5000.5   297.6
  5003.3   297.1  5006.5   297.6  5024.4  303.93  5047.9  303.78  5251.2  303.13
  5274.8  303.72  5436.7  305.82  5506.3  307.33  5621.1  308.73  5723.9  311.35
  5749.7  311.71    5760  307.82  5785.5  307.91  5801.2  312.69  5874.7  319.31
  5951.5  326.71  6017.5  329.03  6130.8  343.45  6274.9  354.16  6562.7  365.24
#Mann= 14 ,-1 , 0
  3940.6     .05       0  3956.6     .08       0  4450.8     .05       0
  4924.9     .12       0  5000.5     .07       0  5006.5     .12       0
  5047.9     .05       0  5251.2      .1       0  5274.8     .05       0
  5436.7     .16       0  5506.3     .05       0  5621.1     .16       0
  5723.9     .12       0  5874.7     .16       0
#XS Ineff= 2 , 0
       0                  5738.8       0  326.14
Permanent Ineff=
       F       F
Bank Sta=4967.5,5024.4
XS Rating Curve= 0 ,0
Exp/Cntr=0.3,0.1

Type RM Length L Ch R = 1 ,111084  ,509,509,509
BEGIN DESCRIPTION:
BIG ELKHART CREEK 124.0
END DESCRIPTION:
XS GIS Cut Line= 3
      3784449.61     10536710.16      3784399.61     10537110.19
      3783899.64     10537660.15
#Sta/Elev= 30
  4625.6   339.3    4744  334.71  4766.7  328.75  4776.8  328.41  4847.3  314.48
  4905.3  305.51    4991   301.7  5005.6   297.8  5008.3   297.3  5011.6   297.8
  5026.2  302.51    5050  303.45  5078.4  300.56  5106.8  301.23  5113.5  299.25
    5121   301.9  5163.6  303.57  5396.7  303.16  5460.9  307.99  5602.1  325.14
  5644.7  326.03  5651.4  328.18  5663.3  328.42  5673.1  328.22  5679.8  330.97
  5687.2  329.28    5694  331.67  5715.6  332.27  5736.6  335.38    5772  335.08
#Mann= 4 ,-1 , 0
  4625.6     .05       0  5005.6     .03       0  5011.6     .05       0
  5663.3     .16       0
Bank Sta=4991,5026.2
XS Rating Curve= 0 ,0
Exp/Cntr=0.3,0.1

Type RM Length L Ch R = 1 ,110575  ,347,347,347
BEGIN DESCRIPTION:
BIG ELKHART CREEK 123.0
END DESCRIPTION:
XS GIS Cut Line= 4
      3784515.51     10536226.85      3784020.72     10536799.77
      3783916.56     10537232.06      3783468.82     10537695.41
#Sta/Elev= 30
  3939.1  371.27  4102.1  355.44  4442.2  330.63  4520.1  327.17  4555.2  327.27
    4598  324.12  4618.8  324.61  4669.2  315.02  4698.9   311.1  4727.4  304.01
  4778.8  302.19  4789.1   298.3  4799.4  297.68  4806.1  301.95    4895  301.31
  4922.8  302.97  4943.4  300.63  4984.5  299.71  5002.1  297.39  5004.9  296.89
  5008.1  297.39  5020.8  302.18  5077.1  299.72  5097.7  301.38  5300.7  327.09
  5327.4  329.18  5554.6  339.59  5589.9  342.65    5604  341.83  5785.1  349.17
#Mann= 5 ,-1 , 0
  3939.1     .05       0  5002.1     .03       0  5008.1     .05       0
  5300.7     .12       0  5327.4     .16       0
Bank Sta=4984.5,5020.8
XS Rating Curve= 0 ,0
Exp/Cntr=0.3,0.1

Type RM Length L Ch R = 1 ,110228  ,1062,1062,1062
BEGIN DESCRIPTION:
BIG ELKHART CREEK 122.0
END DESCRIPTION:
XS GIS Cut Line= 2
      3784277.14     10536202.48      3783228.84     10537625.67
#Sta/Elev= 30
  3930.4  344.11  4005.2     338  4084.6  340.66  4113.9  338.37  4134.7  342.87
  4149.4   342.9  4435.5  332.66  4562.9  308.78  4621.4  301.97  4933.7  300.23
  4970.8  300.98  4984.8  296.15  4996.4   295.7  4999.2   295.2  5002.4   295.7
  5014.1  300.09  5020.5  310.04  5043.3  315.34  5049.5  308.94  5057.8  305.73
  5078.8  310.96    5085  320.52  5093.5  315.06  5099.7  320.95  5120.5   321.4
  5143.6   325.8  5182.8  326.56  5250.1  328.23  5536.2  344.81    5698  349.73
#Mann= 5 ,-1 , 0
  3930.4     .05       0  4933.7     .12       0  4996.4     .07       0
  5002.4     .12       0  5182.8     .16       0
Bank Sta=4970.8,5014.1
XS Rating Curve= 0 ,0
Exp/Cntr=0.3,0.1

Type RM Length L Ch R = 1 ,109166  ,305,305,305
BEGIN DESCRIPTION:
BIG ELKHART CREEK 121.0
END DESCRIPTION:
XS GIS Cut Line= 2
       3783131.3     10535584.41      3782922.96      10537341.4
#Sta/Elev= 30
  4137.8  404.87  4279.5  397.27  4391.1  384.81  4465.9  376.49  4506.1  368.41
  4532.8  359.42  4556.5  360.32  4606.8  355.24  4647.1   338.5  4697.5  326.32
  4703.3  323.06  4757.9  313.11    4768  315.21  4786.1  312.81  4798.2  308.19
  4827.2  305.67  4873.8  298.52  4979.4  299.02  4996.6  294.03  4999.3  293.53
  5002.6  294.03  5019.7  299.68  5032.3  299.08  5190.9  298.42  5362.1  302.27
  5380.4   305.7  5550.9   320.6  5613.9  323.43  5664.2  329.13  5907.1  338.34
#Mann= 7 ,-1 , 0
  4137.8     .05       0  4391.1     .16       0  4827.2     .05       0
  4996.6     .03       0  5002.6     .05       0  5032.3     .12       0
  5613.9     .16       0
Bank Sta=4979.4,5019.7
XS Rating Curve= 0 ,0
Exp/Cntr=0.3,0.1

Type RM Length L Ch R = 1 ,108861  ,525,525,525
BEGIN DESCRIPTION:
BIG ELKHART CREEK 120.0
END DESCRIPTION:
XS GIS Cut Line= 3
      3782799.61     10535760.22      3782749.61     10536510.19
      3782699.61     10537010.17
#Sta/Elev= 30
    4232  399.43  4307.4  389.87  4372.3  378.55  4402.3  376.19  4432.4  365.96
  4502.6  355.53  4522.6  348.96  4542.7  334.86  4592.8  313.99  4602.8  307.78
  4632.9  304.34  4662.9  297.81    4703  297.13  4954.8  298.96  4986.1  297.88
  5000.7   293.8  5003.5   293.3  5006.7   293.8  5023.8  298.68  5036.4  296.39
  5084.1   298.7  5184.6  297.94  5224.8  300.14  5285.1  309.87  5357.8  314.59
  5395.7  317.26  5405.7  313.57  5425.8  317.17  5433.4   321.2  5486.1  324.96
#Mann= 7 ,-1 , 0
    4232     .05       0  4307.4     .16       0  4632.9     .05       0
  4954.8     .12       0  5000.7     .07       0  5006.7     .12       0
  5357.8     .16       0
Bank Sta=4986.1,5023.8
XS Rating Curve= 0 ,0
Exp/Cntr=0.3,0.1

Type RM Length L Ch R = 1 ,108336  ,558,558,558
BEGIN DESCRIPTION:
BIG ELKHART CREEK 119.0
END DESCRIPTION:
XS GIS Cut Line= 3
      3782699.63     10535860.15      3782349.61     10536660.19
      3782399.61     10537060.22
#Sta/Elev= 30
  4131.1  384.66    4169  378.93  4185.7  375.02  4192.3  371.44    4284  357.99
  4320.2  346.89  4327.6  342.66  4343.6  340.16  4349.4  336.35  4360.4  334.07
    4367  329.58  4382.2  325.85    4404  316.44  4419.2  313.86  4442.6  305.43
  4458.4  304.15    4466  302.31  4471.5  304.43    4565  297.08  4820.6  296.21
  4966.5  297.24  4986.9  292.21  4989.7  291.71  4992.9  292.21  5001.6  295.97
  5014.4  297.68  5127.8  296.59  5189.6  309.49  5326.8  324.42  5407.5  328.88
#Mann= 6 ,-1 , 0
  4131.1     .16       0  4458.4     .05       0  4820.6     .12       0
  4986.9     .07       0  4992.9     .12       0  5189.6     .16       0
Bank Sta=4966.5,5001.6
XS Rating Curve= 0 ,0
Exp/Cntr=0.3,0.1

Type RM Length L Ch R = 1 ,107778  ,302,302,302
BEGIN DESCRIPTION:
BIG ELKHART CREEK 118.0
END DESCRIPTION:
XS GIS Cut Line= 3
      3782049.62     10536060.15      3781949.61     10536460.19
      3782199.61     10537010.19
#Sta/Elev= 30
  4572.7  346.13  4595.9  343.28  4624.3  336.19    4632  331.16  4637.2  332.07
  4644.9  330.08  4655.2  324.47  4665.5  322.08  4673.2  316.11  4678.4  317.25
  4686.1  314.74  4696.4  309.29  4706.7  307.04  4714.5  301.53  4719.6  302.41
  4727.4  297.97  4770.4   295.1  4851.1  293.48  4937.9  295.47  4974.7  295.86
  4996.3  291.85  4999.1  291.35  5002.3  291.85  5022.4  295.55  5091.6  294.59
  5348.8  298.07    5431  308.87  5490.3     314  5574.9  324.35  5589.2  324.59
#Mann= 6 ,-1 , 0
  4572.7     .16       0  4770.4     .05       0  4937.9     .12       0
  4996.3     .07       0  5002.3     .12       0  5348.8     .16       0
Bank Sta=4974.7,5022.4
XS Rating Curve= 0 ,0
Exp/Cntr=0.3,0.1

Type RM Length L Ch R = 1 ,107476  ,591,591,591
BEGIN DESCRIPTION:
BIG ELKHART CREEK 117.0
END DESCRIPTION:
XS GIS Cut Line= 3
      3782249.34     10535695.56      3781763.24     10536209.44
      3781409.29     10537305.96
#Sta/Elev= 30
  4105.5  368.76  4172.2  365.12    4243  355.61  4285.5  352.84  4322.3  353.39
  4390.6  353.66  4419.8  352.78  4469.5  347.02  4511.6  335.36  4518.9   335.4
  4525.8  330.87  4582.4  316.29  4589.7  317.04  4610.7  312.29  4671.7  305.75
    4724  297.41  4780.6  293.57  4972.3  294.75  4981.8  295.23  4989.3  291.11
    4992  290.61  4995.3  291.11  5005.9  292.29  5013.3   296.2  5206.7  295.09
  5307.5  296.53  5444.1  312.06  5593.1  320.38  5906.5  329.12  5965.1  327.14
#Mann= 8 ,-1 , 0
  4105.5     .16       0  4322.3     .05       0  4390.6     .16       0
  4671.7     .05       0  4972.3     .12       0  4989.3     .07       0
  4995.3     .12       0  5206.7     .16       0
Bank Sta=4981.8,5013.3
XS Rating Curve= 0 ,0
Exp/Cntr=0.3,0.1

Type RM Length L Ch R = 1 ,106885  ,462,462,462
BEGIN DESCRIPTION:
Mapping XS 6a5f2b03
END DESCRIPTION:
XS GIS Cut Line= 4
      3780770.19     10535015.02      3781075.74     10535876.11
      3781214.62     10536508.05      3781152.41     10536846.76
#Sta/Elev= 30
  3608.7  365.27  3862.3  342.88  3887.9  333.03  3900.7  334.11  3943.1  326.47
  3949.6  329.15  4011.4  330.06  4067.8  340.17  4091.7  340.91  4144.7  336.24
  4195.4  323.73  4247.7  307.59    4253  308.48  4278.6   297.8  4314.8  292.78
  4340.3   296.4  4441.4  294.85  4731.3  294.54    4838     290  4840.8   289.5
    4844     290  4888.6  292.76  4977.1  293.93  4997.6     290  5026.4  290.26
  5031.5  293.75  5094.8  294.57  5354.6  317.78  5435.9  320.06  5513.8  316.56
#Mann= 7 ,-1 , 0
  3608.7     .16       0  4195.4     .12       0  4441.4     .05       0
    4838     .07       0    4844     .05       0  4888.6     .12       0
  5094.8     .16       0
#XS Ineff= 1 ,-1
    3857  4091.7  340.91
Permanent Ineff=
       F
Bank Sta=4977.1,5031.5
XS Rating Curve= 0 ,0
Exp/Cntr=0.3,0.1

Type RM Length L Ch R = 1 ,106423  ,348,348,348
BEGIN DESCRIPTION:
BIG ELKHART CREEK 116.0
END DESCRIPTION:
XS GIS Cut Line= 3
      3780596.57     10535362.21      3780791.01     10535987.22
      3780881.29     10536952.45
#Sta/Elev= 30
  4105.8  364.87  4266.8  356.14  4337.1  342.28  4364.4  346.91    4376  345.33
  4402.2  347.48  4449.3  337.26  4467.2  335.57  4472.5  331.52  4499.8  328.24
    4505  323.45  4522.6  318.29  4537.6  309.61  4564.5  305.21  4575.3  299.52
  4595.9  294.39  4655.2  292.21  4937.4  293.13  4984.3  293.02  4994.3  288.76
  5001.4  288.58  5004.1  288.08  5007.4  288.58  5016.6  292.09  5205.3  292.36
  5245.4  295.41    5278  302.23  5345.9  310.18  5426.4  313.39  5729.8  322.18
#Mann= 7 ,-1 , 0
  4105.8     .16       0  4655.2     .05       0  4937.4     .12       0
  5001.4     .07       0  5007.4     .12       0    5278     .16       0
  5426.4     .05       0
Bank Sta=4984.3,5016.6
XS Rating Curve= 0 ,0
Exp/Cntr=0.3,0.1

Type RM Length L Ch R = 1 ,106075  ,561,561,561
BEGIN DESCRIPTION:
BIG ELKHART CREEK 115.0
END DESCRIPTION:
XS GIS Cut Line= 3
      3780599.61     10535660.22      3780549.61     10536410.19
      3780449.62     10536810.14
#Sta/Elev= 30
  4234.7  354.59  4254.7  355.48  4274.8  354.02  4284.8  351.28  4334.9  346.56
  4425.1  333.27  4445.1  328.34  4475.2  317.78  4555.4  298.67  4565.4  291.91
  4610.9  291.13  4675.6  292.67  4785.9  291.46  4956.3  292.45  4976.3  287.85
  5014.3   287.6    5017   287.1  5020.3   287.6  5027.6  290.95  5045.6  289.94
  5050.8  287.87  5058.5  291.26  5100.9  292.08  5182.2  297.79    5244  305.57
  5264.6  309.52  5339.4  315.49  5348.1  317.37  5380.6  321.14  5398.6  321.56
#Mann= 6 ,-1 , 0
  4234.7     .16       0  4610.9     .12       0  5014.3     .07       0
  5020.3     .12       0  5100.9     .16       0  5348.1     .05       0
Bank Sta=4956.3,5027.6
XS Rating Curve= 0 ,0
Exp/Cntr=0.3,0.1

Type RM Length L Ch R = 1 ,105514  ,464,464,464
BEGIN DESCRIPTION:
BIG ELKHART CREEK 114.0
END DESCRIPTION:
XS GIS Cut Line= 3
       3780399.6     10535660.21      3780049.61     10536360.19
      3780149.61     10536760.18
#Sta/Elev= 30
  4212.1  356.63  4270.8  351.84  4293.1  347.51  4301.5  344.32  4315.5  341.92
  4323.9  337.32  4332.3  335.51    4377  317.55    4391  314.79  4404.9  309.31
  4421.7  306.41  4435.7   301.2  4445.6  299.84    4458  296.59  4494.4  292.14
  4829.8  290.33  4972.3  291.57  4980.7  287.46  5009.7  286.89  5012.5  286.39
  5015.7  286.89  5025.6  291.17  5086.3   300.3  5100.4  300.35  5124.5  303.44
  5186.7  308.21  5234.4  311.72  5306.5  316.47  5334.9  320.29    5407  323.39
#Mann= 9 ,-1 , 0
  4212.1     .16       0  4445.6     .05       0  4829.8     .12       0
  5009.7     .07       0  5015.7     .12       0  5086.3     .16       0
  5124.5     .12       0  5186.7     .16       0  5234.4     .05       0
Bank Sta=4972.3,5025.6
XS Rating Curve= 0 ,0
Exp/Cntr=0.3,0.1

Type RM Length L Ch R = 1 ,105050  ,664,664,664
BEGIN DESCRIPTION:
BIG ELKHART CREEK 113.0
END DESCRIPTION:
XS GIS Cut Line= 3
       3779349.6     10535360.17      3779599.61     10536160.19
      3779749.62     10536560.22
#Sta/Elev= 30
  4081.6  402.39  4200.5  383.47  4249.2  368.14  4303.2  358.23  4330.4  341.55
  4362.9  332.68  4368.2  335.12    4375  328.51  4416.9  312.96  4488.9  291.01
  4530.6  287.67  4718.8   289.8    4794  286.97  4806.1  290.11  4856.9  289.99
  4865.8  285.63  4871.1  290.19  4914.1  285.59  4916.9  285.09  4920.1  285.59
  4965.2  291.16  4973.2  286.83  4990.1  285.92    5015   290.4  5080.9  289.62
  5100.4  293.85  5105.8  291.43  5122.7  300.97  5213.2  311.84    5347  317.84
#Mann= 6 ,-1 , 0
  4081.6     .16       0  4488.9     .05       0  4718.8     .12       0
  4914.1     .07       0  4920.1     .12       0  5213.2     .05       0
Bank Sta=4965.2,5015
XS Rating Curve= 0 ,0
Exp/Cntr=0.3,0.1

Type RM Length L Ch R = 1 ,104386  ,483,483,483
BEGIN DESCRIPTION:
BIG ELKHART CREEK 112.0
END DESCRIPTION:
XS GIS Cut Line= 3
       3779099.6     10535560.14      3779149.61     10535960.19
      3779549.59     10536510.16
#Sta/Elev= 30
  4567.9  370.76  4588.1  367.85  4598.2  364.37  4605.7  363.28  4610.8  364.86
  4638.5  358.62  4668.7   356.1  4678.8  353.37    4709  343.42  4719.1  336.65
  4749.3  324.46  4759.4  315.63  4779.6  306.61  4819.9  298.12  4860.2  293.08
  4919.2  289.67  4984.6  287.71  4996.3  284.61    4999  284.11  5002.3  284.61
    5014  289.16  5078.9  287.71  5472.2  291.84  5486.9  295.74  5493.1  295.51
  5501.6   299.7  5549.9  306.34    5558  306.04  5587.4  310.97  5651.1  313.56
#Mann= 5 ,-1 , 0
  4567.9     .16       0  4919.2     .12       0  4996.3     .07       0
  5002.3     .12       0  5549.9     .05       0
Bank Sta=4984.6,5014
XS Rating Curve= 0 ,0
Exp/Cntr=0.3,0.1

Type RM Length L Ch R = 1 ,103903  ,559,559,559
BEGIN DESCRIPTION:
BIG ELKHART CREEK 111.0
END DESCRIPTION:
XS GIS Cut Line= 3
      3778749.61      10535710.2      3778799.61     10536310.19
      3778699.61     10537110.19
#Sta/Elev= 30
  4435.1  358.81  4485.3  351.83  4492.8  347.88  4497.8  350.47  4505.3  346.77
  4525.4  341.22  4535.4  335.13  4565.5  324.86  4613.2   303.8  4618.2   304.6
  4655.9  293.32    4686  286.89  4708.2  287.94  4979.5  288.53    4994  284.02
  4996.8  283.52    5000  284.02  5017.1   287.9  5206.6  287.03  5369.7     287
  5434.1  289.37  5478.1  292.92    5531   294.1  5631.8   304.2  5644.4   302.8
  5651.9  305.14  5682.2  308.54  5712.4  314.81  5742.6  318.86  5843.4  327.97
#Mann= 6 ,-1 , 0
  4435.1     .16       0  4708.2     .05       0    4994     .03       0
    5000     .05       0  5206.6     .12       0  5434.1     .05       0
Bank Sta=4979.5,5017.1
XS Rating Curve= 0 ,0
Exp/Cntr=0.3,0.1

Type RM Length L Ch R = 1 ,103344  ,358,358,358
BEGIN DESCRIPTION:
BIG ELKHART CREEK 110.0
END DESCRIPTION:
XS GIS Cut Line= 3
      3778699.62     10535560.17      3778249.61     10536260.19
      3777849.61     10536760.19
#Sta/Elev= 30
  4180.5  369.84  4239.6  365.95  4297.1  351.67    4303  347.78  4318.2  346.24
  4333.4  342.88  4339.4  339.13  4369.7  333.99  4396.8  320.51    4412  317.05
  4433.1  307.95  4510.7  293.24  4557.3   287.4    4630  285.61  4989.9  286.99
  4996.1  283.16  4998.9  282.66  5002.1  283.16  5019.9  287.24  5076.7  285.95
  5346.3  289.06  5389.7  290.59  5404.1  286.54  5410.5  288.64  5418.5  287.44
  5447.3  293.09  5453.7  299.38  5468.1  301.95  5576.2  309.37    5653  316.33
#Mann= 6 ,-1 , 0
  4180.5     .16       0  4510.7     .16       0  4996.1     .03       0
  5002.1     .16       0  5346.3     .12       0  5576.2     .16       0
Bank Sta=4989.9,5019.9
XS Rating Curve= 0 ,0
Exp/Cntr=0.3,0.1

Type RM Length L Ch R = 1 ,102986  ,775,775,775
BEGIN DESCRIPTION:
BIG ELKHART CREEK 109.0
END DESCRIPTION:
XS GIS Cut Line= 4
      3778688.38     10535225.68      3778059.01     10535772.58
      3777898.42     10536597.23      3777647.88     10536856.41
#Sta/Elev= 30
  3830.1  369.34    3875  365.94  3967.1  365.53  4101.9  354.07  4208.3  337.98
  4214.9  333.16  4222.5  333.31  4229.1  328.22    4251  324.69  4257.6  319.11
  4265.3  318.86    4307  304.13  4409.9  289.91    4692   291.2  4956.9  287.77
  4996.7  282.37  5048.3  286.43  5055.8  281.51  5058.5  281.01  5061.8  281.51
  5089.3  285.54  5333.1  288.02  5363.2  289.34  5374.6  285.48  5384.8  289.06
  5405.2   290.1  5435.7  300.24  5483.6  304.82  5696.2  316.37  5864.5  313.56
#Mann= 6 ,-1 , 0
  3830.1     .16       0  4409.9     .16       0  5055.8     .07       0
  5061.8     .16       0  5333.1     .12       0  5483.6     .16       0
#XS Ineff= 2 , 0
         4897.73  304.53
Permanent Ineff=
       F       F
Bank Sta=4956.9,5089.3
XS Rating Curve= 0 ,0
Exp/Cntr=0.3,0.1
