HEC-RAS study BIG ELKHART CREEK.prj: BIG ELKHART CREEK Base Level Engineering

--- BIG ELKHART CREEK.g01 (geometry) --- (continued)

Type RM Length L Ch R = 1 ,102211  ,800,800,800
BEGIN DESCRIPTION:
BIG ELKHART CREEK 108.0
END DESCRIPTION:
XS GIS Cut Line= 3
      3777442.69     10534761.24      3777516.48     10535959.21
      3777494.78     10537052.96
#Sta/Elev= 30
    3543  343.04    3582  341.93  3642.1  335.29  3732.1  312.06  3822.5  306.06
  3903.6  305.62  4060.1  296.33  4226.6   293.8  4373.5  287.25  4894.2   285.1
  4964.3  287.32  4981.3  281.23    4984  280.73  4987.3  281.23  4994.3   281.5
  5004.3  286.06  5064.3  288.22  5174.3  286.67  5194.3  289.96  5234.3  302.06
  5284.3  305.03    5331  307.43  5554.4  304.04  5564.4  300.96  5574.4  301.92
  5594.4  297.88  5604.4  299.05  5614.4  304.48  5634.4  309.48  5837.2  319.48
#Mann= 6 ,-1 , 0
    3543     .16       0  3903.6     .16       0  4981.3     .07       0
  4987.3     .16       0  5284.3     .05       0    5331     .16       0
#XS Ineff= 2 , 0
         4900.57   302.6
Permanent Ineff=
       F       F
Bank Sta=4964.3,5004.3
XS Rating Curve= 0 ,0
Exp/Cntr=0.3,0.1

Type RM Length L Ch R = 1 ,101411  ,604,604,604
BEGIN DESCRIPTION:
BIG ELKHART CREEK 107.0
END DESCRIPTION:
XS GIS Cut Line= 3
       3776849.6     10535460.17      3777049.61     10535810.19
      3777249.62     10536910.22
#Sta/Elev= 30
  4589.1  356.02  4656.1  349.39  4661.8  346.39  4677.7  345.81  4683.4  342.76
  4736.7  340.81  4758.3  336.57  4779.9  328.17  4785.6  328.37    4808  320.55
  4838.9  305.67  4888.6  289.95  4962.7  280.85  4969.2  285.05  4984.3  283.83
  4986.4  279.81  4989.1  279.31  4992.4  279.81  5002.4  279.86  5012.6  285.72
  5072.3  287.24  5124.4     285  5195.5  286.69  5378.5  285.12  5591.9  287.89
  5694.8  289.66  5795.2  299.03  5828.7  302.28  6072.9  320.36  6110.3  321.32
#Mann= 7 ,-1 , 0
  4589.1     .16       0  4736.7     .16       0  4986.4     .07       0
  4992.4     .16       0  5795.2      .1       0  5828.7     .16       0
  6072.9     .05       0
Bank Sta=4984.3,5012.6
XS Rating Curve= 0 ,0
Exp/Cntr=0.3,0.1

Type RM Length L Ch R = 1 ,100807  ,1092,1092,1092
BEGIN DESCRIPTION:
BIG ELKHART CREEK 106.0
END DESCRIPTION:
XS GIS Cut Line= 3
       3776599.6     10535710.16      3776649.61     10536110.19
      3776799.61     10536710.18
#Sta/Elev= 30
  4577.9  348.81  4615.7   341.5  4628.3  333.23  4638.4  330.82  4648.5  325.15
  4658.6  322.36  4668.6  316.16  4678.7  313.58  4688.8  307.02  4701.4  303.45
  4708.9  299.47  4749.3  290.17  4785.4  285.48    4840  283.55  4870.2   285.3
    4935   285.2    4971  283.75  4983.6  281.13  4996.1  278.27  4998.8  277.77
  5002.1  278.27    5012   279.2  5022.3  283.32  5032.6  284.75  5169.2  282.85
  5299.2  283.67  5352.1  284.31  5444.9  291.25  5503.4  298.56  5599.5  309.59
#Mann= 7 ,-1 , 0
  4577.9     .16       0  4785.4     .05       0    4935     .12       0
  4996.1     .07       0  5002.1     .12       0  5299.2      .1       0
  5503.4     .16       0
Bank Sta=4983.6,5022.3
XS Rating Curve= 0 ,0
Exp/Cntr=0.3,0.1

Type RM Length L Ch R = 1 ,99715   ,432,432,432
BEGIN DESCRIPTION:
BIG ELKHART CREEK 105.0
END DESCRIPTION:
XS GIS Cut Line= 3
       3776366.3     10535620.67      3776084.18      10536184.9
      3776192.51     10536986.48
#Sta/Elev= 30
  4050.4  358.24  4099.5  353.71  4105.8  350.71  4121.9  348.72  4128.1   344.8
  4143.6  343.15    4161  331.79  4166.6  332.08  4183.4  324.18    4189  324.08
  4205.8  314.53  4211.3  314.66  4239.9   302.6  4276.7  295.27  4284.7  291.76
    4307  288.92  4374.1  286.37  4541.2  286.13  4777.4  280.89    4959  282.31
  4983.7  278.46  4986.3  276.04    4989  275.54  4992.3  276.04  4993.1  276.26
  5009.5  282.16    5070   293.6  5291.6  312.48    5403  316.08  5490.1  312.45
#Mann= 6 ,-1 , 0
  4050.4     .16       0  4276.7     .05       0  4986.3     .07       0
  4992.3     .05       0  4993.1     .12       0  5291.6     .16       0
Bank Sta=4959,5009.5
XS Rating Curve= 0 ,0
Exp/Cntr=0.3,0.1

Type RM Length L Ch R = 1 ,99283   ,86,86,86
BEGIN DESCRIPTION:
Mapping XS bd7ba50b
END DESCRIPTION:
XS GIS Cut Line= 4
        3776388.     10535507.82      3775702.24     10536137.16
      3775754.32     10536597.23      3776088.52     10536944.45
#Sta/Elev= 30
  3650.6  352.81  3658.3  350.18  3679.3  353.45  3686.7  351.26  3693.5  354.53
  3721.9  353.66  3750.2  346.83  3806.9  341.49  3813.7  343.41  3821.1  338.17
  3870.5  331.72  3877.9  327.11  3884.6  329.23    3892  323.68    3913  319.16
  3941.4   306.5  4004.9   296.7  4213.8  292.36  4549.9  283.97  4925.5  280.28
  4954.7  279.91  4959.9  279.74  5004.1  275.23  5006.9  274.73  5010.1  275.23
  5037.3   283.8  5128.4  294.61  5157.7  296.69  5410.8   311.8  5526.3   313.1
#Mann= 8 ,-1 , 0
  3650.6     .16       0  4213.8     .05       0  4925.5     .12       0
  4954.7     .05       0  5004.1     .04       0  5010.1     .05       0
  5128.4     .12       0  5157.7     .16       0
Bank Sta=4959.9,5037.3
XS Rating Curve= 0 ,0
Exp/Cntr=0.3,0.1

Type RM Length L Ch R = 1 ,99197   ,262,262,262
BEGIN DESCRIPTION:
Mapping XS 1851ac44
END DESCRIPTION:
XS GIS Cut Line= 5
      3775346.35     10535507.86      3775667.52     10536319.45
      3775689.22     10536614.59      3775684.88     10536718.76
       3775741.3     10537269.96
#Sta/Elev= 30
  3938.3  361.09  3954.4  359.86  3988.6  356.52  4059.1  329.93  4102.1  319.34
  4234.5  301.09  4252.7  296.01  4339.6  287.25  4475.1  282.39  4521.5  283.32
  4543.1   286.7  4553.9  285.18    4767     282  4972.3  280.75  4989.4  274.84
  4992.1  274.34  4995.4  274.84  5002.4  275.06  5012.4  280.65  5107.1  283.84
  5132.7  291.47  5190.7  294.77  5278.2  295.02  5343.4  294.44  5373.6  288.55
  5401.9   295.6  5660.4  317.02    5700  317.18  5715.4  320.93  5765.4   322.5
#Mann= 10 ,-1 , 0
  3938.3     .05       0  3954.4     .16       0  4339.6     .05       0
  4553.9     .12       0    4767     .05       0  4989.4     .04       0
  4995.4     .05       0  5190.7     .12       0  5278.2     .16       0
  5660.4     .05       0
Bank Sta=4972.3,5012.4
XS Rating Curve= 0 ,0
Exp/Cntr=0.3,0.1

Type RM Length L Ch R = 1 ,98935   ,793,793,793
BEGIN DESCRIPTION:
BIG ELKHART CREEK 104.0
END DESCRIPTION:
XS GIS Cut Line= 3
      3775168.38     10535559.87       3775428.8     10536362.85
      3775545.99     10537209.22
#Sta/Elev= 30
  4054.6  369.32  4104.7  368.13  4149.5  360.29  4168.7  353.63  4223.1  325.06
  4264.6   310.7  4296.6  302.77  4353.9  297.64  4383.2  292.93  4493.7  283.01
  4653.6  279.43  4966.7  281.24  4976.8  276.75  5004.1  274.66  5006.9  274.16
  5010.1  274.66  5013.1     280  5018.1  277.01  5057.6  281.57  5128.3  280.24
  5259.5  284.06  5305.3   289.7  5441.2  296.28  5461.4  299.81  5511.9  301.22
  5575.7  307.34  5592.4  310.65  5597.5   307.9  5701.6  315.97  5753.2  317.64
#Mann= 8 ,-1 , 0
  4054.6     .16       0  4353.9     .08       0  4383.2     .05       0
  4653.6     .12       0  5004.1     .07       0  5010.1     .12       0
  5575.7     .16       0  5701.6     .05       0
Bank Sta=4966.7,5013.1
XS Rating Curve= 0 ,0
Exp/Cntr=0.3,0.1

Type RM Length L Ch R = 1 ,98142   ,670,670,670
BEGIN DESCRIPTION:
BIG ELKHART CREEK 103.0
END DESCRIPTION:
XS GIS Cut Line= 3
      3774649.59     10535860.15      3774899.61     10536460.19
      3775443.56     10537516.41
#Sta/Elev= 30
  4380.1  368.29  4412.6  366.07    4424  358.14  4447.8  352.72  4477.6  335.83
  4488.5  333.53  4510.1  325.03  4519.3  318.99    4586  294.01  4625.5  286.56
  4691.4  281.96  4755.5  277.33  4856.1  276.62  4986.3  278.61  4994.6  272.84
  4997.4  272.34  5000.6  272.84  5015.5  272.94  5020.9  278.03  5476.2  277.53
  5563.7  280.65  5690.3  289.59  5802.9  299.03  5915.4  307.38  5936.1  305.88
  6024.8  314.39  6107.8  316.44  6179.9  323.88  6196.5  320.91  6218.2  322.14
#Mann= 9 ,-1 , 0
  4380.1     .16       0  4691.4     .05       0  4856.1     .12       0
  4994.6     .07       0  5000.6     .12       0  5563.7     .05       0
  5690.3     .16       0  5802.9     .08       0  5915.4     .05       0
Bank Sta=4986.3,5020.9
XS Rating Curve= 0 ,0
Exp/Cntr=0.3,0.1

Type RM Length L Ch R = 1 ,97472   ,517,517,517
BEGIN DESCRIPTION:
BIG ELKHART CREEK 102.0
END DESCRIPTION:
XS GIS Cut Line= 3
       3774599.6     10535860.22      3774449.61     10536410.19
      3774734.22      10537785.8
#Sta/Elev= 30
  4433.2  372.15  4455.6  369.18  4474.6  363.86  4524.7  340.22  4536.8  330.19
  4547.2  328.95  4578.3  312.59    4599  306.51  4609.4  298.69  4630.1   290.8
  4671.6  280.34  4721.3   277.5  4858.1  278.26    4927   276.4    4986  276.22
  4989.9   271.1  4992.6   270.6  4995.9   271.1  5013.5  271.34  5033.9   277.5
  5268.8  276.18  5738.5  278.26  5916.8  284.05  5936.4  287.42    6004  290.61
  6033.1  289.94  6055.1  288.91  6075.5  292.17    6258  307.25    6408  317.11
#Mann= 7 ,-1 , 0
  4433.2     .16       0  4721.3     .05       0    4927     .12       0
  4989.9     .07       0  4995.9     .12       0  5936.4     .05       0
  6033.1     .16       0
Bank Sta=4986,5033.9
XS Rating Curve= 0 ,0
Exp/Cntr=0.3,0.1

Type RM Length L Ch R = 1 ,96955   ,724,724,724
BEGIN DESCRIPTION:
BIG ELKHART CREEK 101.0
END DESCRIPTION:
XS GIS Cut Line= 4
       3774478.3     10535750.84      3774078.98     10536449.66
      3774139.74     10536901.05      3773749.12     10537751.72
#Sta/Elev= 30
  4040.3  369.96  4089.7  360.85  4177.8   323.6  4223.6  310.96  4272.6  292.66
    4316   282.5  4364.3  279.11  4810.1  277.09  4967.1  276.81  5004.1  270.15
  5006.9  269.65  5010.1  270.15  5017.2  277.03  5112.7  274.21  5429.5  278.84
  5442.7  275.35    5458  278.91  5519.8  279.62  5526.9  277.14  5532.4     280
  5541.8  276.31  5578.4  276.42  5662.8  286.33  5732.7  286.46  5838.8  290.33
  5888.2  293.91  5911.2   291.1  5944.9  295.07  6031.6  295.85  6236.7   305.4
#Mann= 8 ,-1 , 0
  4040.3     .16       0  4364.3     .05       0  4810.1     .12       0
  5004.1     .07       0  5010.1     .12       0  5732.7     .16       0
  5838.8     .05       0  5944.9     .16       0
Bank Sta=4967.1,5017.2
XS Rating Curve= 0 ,0
Exp/Cntr=0.3,0.1

Type RM Length L Ch R = 1 ,96231   ,403,403,403
BEGIN DESCRIPTION:
BIG ELKHART CREEK 100.0
END DESCRIPTION:
XS GIS Cut Line= 3
      3774161.44     10535403.66      3773618.91     10536315.11
      3773514.74     10537712.63
#Sta/Elev= 30
  3674.2  338.22    3709  334.73  3724.6  328.15  3730.4  329.09    3740  326.64
    3746  318.89  3751.8  320.32  3767.4  318.56  3774.9  315.55  3798.2  312.57
  3921.3  301.33  4065.8  294.34  4154.9  285.02    4299  284.18  4760.1  274.09
  4980.7   274.7  4984.3  273.43  4997.7  269.43  5000.5  268.93  5003.7  269.43
  5010.7  269.45  5030.8  275.56  5351.7  274.08  5567.5     281  5712.7  291.57
  5808.1  295.36  5907.9     299  5943.3  304.06  6053.6  306.79  6136.3  312.27
#Mann= 7 ,-1 , 0
  3674.2     .05       0  4984.3     .12       0  4997.7     .07       0
  5003.7     .12       0  5567.5     .16       0  5808.1     .05       0
  5907.9     .16       0
Bank Sta=4980.7,5030.8
XS Rating Curve= 0 ,0
Exp/Cntr=0.3,0.1

Type RM Length L Ch R = 1 ,95828   ,714,714,714
BEGIN DESCRIPTION:
BIG ELKHART CREEK 99.0
END DESCRIPTION:
XS GIS Cut Line= 3
      3772967.87     10535507.85      3773319.43     10536844.62
      3773219.67     10537655.68
#Sta/Elev= 30
  3755.1  376.09  3863.6  367.68  3938.7  354.26  3943.8  348.98  3973.8  342.95
    3979  336.54  4005.7  330.67  4014.2  327.37  4019.3  322.38    4047  315.92
  4059.7  307.98  4088.4  301.51    4100   293.6  4119.4  287.63  4140.4  283.32
    4220  276.44  4574.4  272.21  4865.4  273.75  4967.3  274.93  4993.8  267.91
  4996.5  267.41  4999.8  267.91  5008.7  268.84    5019  274.52  5172.5  272.28
  5304.1  275.04  5485.1  287.79  5686.6  293.48  5789.3   298.7  5954.5  307.07
#Mann= 9 ,-1 , 0
  3755.1      .1       0  3863.6     .16       0    4220     .05       0
  4865.4     .12       0  4993.8     .07       0  4999.8     .12       0
  5485.1     .16       0  5686.6     .05       0  5789.3     .16       0
Bank Sta=4967.3,5019
XS Rating Curve= 0 ,0
Exp/Cntr=0.3,0.1

Type RM Length L Ch R = 1 ,95114   ,665,665,665
BEGIN DESCRIPTION:
BIG ELKHART CREEK 98.0
END DESCRIPTION:
XS GIS Cut Line= 3
      3772781.24     10535412.37      3772855.02     10537022.58
      3773011.23     10537595.36
#Sta/Elev= 30
    3550  381.79    3728  378.59  3788.1  374.47  3817.2  369.43  3858.1  364.66
  3928.2  339.52  3938.2  339.85  3968.3  327.38  4018.3  311.35  4048.3  298.18
    4062   295.7  4068.4  291.35  4088.4  284.27  4108.4  280.33  4172.7  274.35
  4325.3  273.74  4412.4   272.8  4717.3  271.88  4979.3  272.69  5006.3  266.23
  5009.1  265.73  5012.3  266.23  5019.4  272.01  5129.5  272.94  5190.5  279.99
  5300.2  283.64  5532.6  292.55  5547.2  295.07  5654.4  302.68  5755.6  306.86
#Mann= 11 ,-1 , 0
    3550      .1       0  3817.2     .16       0  4172.7     .05       0
  4325.3     .08       0  4412.4     .05       0  4717.3     .12       0
  5006.3     .07       0  5012.3     .12       0  5300.2     .16       0
  5547.2     .05       0  5654.4     .16       0
Bank Sta=4979.3,5019.4
XS Rating Curve= 0 ,0
Exp/Cntr=0.3,0.1

Type RM Length L Ch R = 1 ,94449   ,610,610,610
BEGIN DESCRIPTION:
BIG ELKHART CREEK 97.0
END DESCRIPTION:
XS GIS Cut Line= 3
      3771849.64     10535910.23      3772399.61     10536710.19
      3772949.61     10537510.19
#Sta/Elev= 30
    4008   348.8  4036.4  341.47  4066.1  324.88  4087.1  323.17    4123  313.14
  4179.8  302.84  4338.1  281.93  4367.9  279.71  4386.9  281.07  4568.2  272.54
  4649.2   271.1  4769.2  270.13  4929.4  271.93  4992.3  269.76  5001.1  264.57
  5012.2  264.21  5014.9  263.71  5018.2  264.21  5022.1  270.09  5294.3  271.07
  5439.7   280.9  5604.6   285.3  5640.4  289.12  5655.3  288.18  5670.2  292.62
  5676.3  289.27  5697.2  289.53  5810.7  295.18  5935.7  301.65  5949.6  302.33
#Mann= 10 ,-1 , 0
    4008     .16       0  4386.9     .05       0  4568.2     .08       0
  4649.2     .05       0  4769.2     .12       0  5012.2     .07       0
  5018.2     .12       0  5439.7     .16       0  5810.7     .05       0
  5935.7     .16       0
Bank Sta=4992.3,5022.1
XS Rating Curve= 0 ,0
Exp/Cntr=0.3,0.1

Type RM Length L Ch R = 1 ,93839   ,570,570,570
BEGIN DESCRIPTION:
BIG ELKHART CREEK 96.0
END DESCRIPTION:
XS GIS Cut Line= 4
      3771548.61     10535971.39      3771907.97     10536606.78
       3771991.3      10536997.4      3772474.71     10538114.95
#Sta/Elev= 30
  4117.9  357.06  4185.4   348.7  4191.1  344.95    4207  343.83  4212.8  338.55
  4250.3  334.16    4256  330.68  4271.9  327.81  4277.7  323.38  4315.2  317.49
  4331.1  317.91  4336.9  314.82  4352.8  315.87  4358.5  312.95  4476.4  299.99
  4778.6  272.88  4904.9  269.44  4977.4  270.72  5001.7  263.43  5004.5  262.93
  5007.7  263.43    5015  264.07  5021.8  270.86  5337.5   267.4  5709.3  271.33
  5812.2  274.18  5849.6  274.71  5947.6  282.39  6154.6  305.85  6464.9  317.41
#Mann= 7 ,-1 , 0
  4117.9     .16       0  4476.4     .05       0  4904.9     .12       0
  5001.7     .07       0  5007.7     .12       0  5709.3     .05       0
  5812.2     .16       0
Bank Sta=4977.4,5021.8
XS Rating Curve= 0 ,0
Exp/Cntr=0.3,0.1

Type RM Length L Ch R = 1 ,93269   ,599,599,599
BEGIN DESCRIPTION:
BIG ELKHART CREEK 95.0
END DESCRIPTION:
XS GIS Cut Line= 3
      3771149.61      10536210.2      3771499.61     10536910.19
      3772449.62     10538460.21
#Sta/Elev= 30
    4239  379.15  4261.3  375.83  4283.7  368.28  4336.8  346.11  4381.5  336.18
  4409.5  325.23  4417.9  319.44  4448.6   311.9  4454.2  306.53    4485  297.23
  4521.3  291.12  4694.6  271.23  4775.6  267.36  4903.8  268.34  4976.9  268.95
  4996.2  261.22    4999  260.72  5002.2  261.22  5007.6  261.48  5013.2  268.66
  5537.7  266.61  5757.8  269.45  5885.9  275.22  6025.3  284.53  6040.8  284.21
  6046.6  280.53  6083.4   287.7  6382.2  312.09  6735.3  325.62  6839.6  329.99
#Mann= 7 ,-1 , 0
    4239     .16       0  4903.8     .12       0  4996.2     .07       0
  5002.2     .12       0  5757.8     .05       0  5885.9     .16       0
  6735.3     .05       0
Bank Sta=4976.9,5013.2
XS Rating Curve= 0 ,0
Exp/Cntr=0.3,0.1

Type RM Length L Ch R = 1 ,92670   ,558,558,558
BEGIN DESCRIPTION:
BIG ELKHART CREEK 94.0
END DESCRIPTION:
XS GIS Cut Line= 2
      3770131.95      10536169.3      3771985.36     10538277.81
#Sta/Elev= 30
  3712.2  396.38  3760.8  390.87  3775.1  384.05  3810.2  375.33  3817.7  367.32
  3846.2  354.54  3895.6   337.3  3902.2  338.21  3938.2  321.33  4030.3  304.05
  4242.8  280.61  4537.5  271.96  4625.2  272.45  4878.3  265.93  4972.5  267.35
  4990.4  260.17  4993.1  259.67  4996.4  260.17  5000.9  260.52  5007.6  265.97
  5348.2  265.47  5652.8  270.53    5735  269.32  5828.2  272.66  5870.1  275.16
  6049.4  299.97  6275.7     308  6402.2  310.82  6410.9  310.94  6519.5  314.15
#Mann= 11 ,-1 , 0
  3712.2     .16       0  4537.5     .05       0  4878.3     .12       0
  4990.4     .07       0  4996.4     .12       0    5735     .08       0
  5828.2     .05       0  5870.1     .16       0  6275.7     .05       0
  6402.2     .16       0  6410.9     .05       0
Bank Sta=4972.5,5007.6
XS Rating Curve= 0 ,0
Exp/Cntr=0.3,0.1

Type RM Length L Ch R = 1 ,92112   ,571,571,571
BEGIN DESCRIPTION:
BIG ELKHART CREEK 93.0
END DESCRIPTION:
XS GIS Cut Line= 3
      3770049.59     10536510.15      3770499.61     10537310.19
      3770899.59     10538110.15
#Sta/Elev= 30
  4082.3  315.32    4112  310.61    4177  293.88  4214.6  286.72  4376.5  270.74
  4449.5  266.72  4517.5  265.49  4684.4  265.86  4713.4  264.25  4793.7  266.29
  4915.9  265.04  4977.3  265.66  4983.5  260.01  4986.3  259.51  4989.5  260.01
    5003  260.72  5008.6  265.55  5321.7  264.08    5372  265.72  5402.7  262.82
  5461.4  265.76  5657.1  267.03  5693.4  269.65  5707.4  273.03  5736.3  274.53
  5813.6  283.58  5849.9  284.46  5858.3  287.41  5880.7   289.1  5894.6  292.79
#Mann= 6 ,-1 , 0
  4082.3     .16       0  4517.5     .05       0  4915.9     .12       0
  4983.5     .07       0  4989.5     .12       0  5736.3     .05       0
Bank Sta=4977.3,5008.6
XS Rating Curve= 0 ,0
Exp/Cntr=0.3,0.1

Type RM Length L Ch R = 1 ,91541   ,522,522,522
BEGIN DESCRIPTION:
BIG ELKHART CREEK 92.0
END DESCRIPTION:
XS GIS Cut Line= 3
      3769549.59     10536910.17      3769949.61     10537360.19
       3770899.6     10538310.18
#Sta/Elev= 30
  4406.7  305.76    4428  304.15  4463.2  297.57  4540.9  287.19  4576.9  285.04
  4647.6  275.25    4739  267.14  4810.2  263.89  4987.5  264.21    4992  259.24
  4994.8  258.74    4998  259.24  5001.7  259.47  5005.5  262.76  5022.9  264.31
  5305.8  264.77  5334.1  262.12  5348.2  264.26  5404.8  264.48  5701.8  265.07
  5715.9  262.37  5730.1  264.83  5984.6  264.12  6041.2  268.58  6097.7  275.42
  6111.9  274.48  6140.2  281.06  6177.5  285.46  6281.6  300.59  6352.3  306.34
#Mann= 5 ,-1 , 0
  4406.7     .16       0    4739     .12       0    4992     .07       0
    4998     .12       0  6177.5     .16       0
Bank Sta=4987.5,5022.9
XS Rating Curve= 0 ,0
Exp/Cntr=0.3,0.1

Type RM Length L Ch R = 1 ,91019   ,1052,1052,1052
BEGIN DESCRIPTION:
BIG ELKHART CREEK 91.0
END DESCRIPTION:
XS GIS Cut Line= 3
      3769485.03     10536953.46      3769699.61     10537660.19
      3770799.58     10538610.17
#Sta/Elev= 30
  4287.9  309.63    4321  308.96  4368.1  303.71  4490.6  295.69  4574.6  282.55
  4671.2  266.58    4713   263.2  4932.4  262.06  4977.2  263.33  4992.1   257.3
  4994.9   256.8  4998.1   257.3    5010  257.76    5016  263.18  5211.3  263.52
  5238.8   260.8  5281.5  263.66  5473.5  261.36  5813.5  263.97  5983.6  262.51
  6054.9  264.97  6069.1  267.89  6167.7  277.76  6239.1  285.86  6366.4  297.08
  6374.1  299.56    6430   301.1  6437.7  304.16  6458.5  307.23  6479.9  307.92
#Mann= 5 ,-1 , 0
  4287.9     .16       0  4574.6     .12       0  4992.1     .07       0
  4998.1     .12       0  6167.7     .16       0
Bank Sta=4977.2,5016
XS Rating Curve= 0 ,0
Exp/Cntr=0.3,0.1

Type RM Length L Ch R = 1 ,89967   ,652,652,652
BEGIN DESCRIPTION:
BIG ELKHART CREEK 90.0
END DESCRIPTION:
XS GIS Cut Line= 2
      3768482.44     10537057.67      3770005.24     10539270.28
#Sta/Elev= 30
  3398.4  308.76  3425.8  309.25  3506.3   305.4  3512.4  306.88  3542.2  304.32
  3563.2  305.33  3715.4  297.54  3787.1  290.66  3850.6  287.88  3909.5  280.18
  3987.3  266.58    4017  263.62  4139.9   260.5  4987.7     260  4990.7  255.35
  4993.5  254.85  4996.7  255.35  5008.6  256.04    5016  259.67  5246.7  261.31
    5382  260.27  5440.9  264.91    5510  267.41    5591  274.89  5605.9  278.51
  5835.9  303.54  5886.6  305.68  5892.7  304.28  5928.5  305.13  6084.4  313.03
#Mann= 5 ,-1 , 0
  3398.4     .16       0  4139.9     .12       0  4990.7     .07       0
  4996.7     .12       0    5510     .16       0
Bank Sta=4987.7,5016
XS Rating Curve= 0 ,0
Exp/Cntr=0.3,0.1

Type RM Length L Ch R = 1 ,89315   ,554,554,554
BEGIN DESCRIPTION:
BIG ELKHART CREEK 89.0
END DESCRIPTION:
XS GIS Cut Line= 3
      3768299.63     10537610.23      3768749.61     10538410.19
      3769249.59     10539210.16
#Sta/Elev= 30
  4058.7  290.05  4104.2  285.26  4206.9  279.89  4368.4  264.42  4492.5  259.11
  4558.1  257.26  4563.8  258.59  4595.7  257.22  4873.3  257.65  4884.6  253.59
  4887.4  253.09  4890.6  253.59  4896.2   258.4  4979.5  258.87  4990.1  255.12
  5005.4  255.27  5011.9  261.25  5020.8  261.96  5057.3  258.08  5084.4   257.5
  5448.2  260.61  5455.9  259.12  5534.9  258.75  5665.8  261.78  5717.7  260.95
  5781.4  266.14  5844.5  274.59  5884.6  280.28    5891  283.01  5919.9  285.33
#Mann= 5 ,-1 , 0
  4058.7     .16       0  4492.5     .12       0  4884.6     .07       0
  4890.6     .12       0  5844.5     .16       0
Bank Sta=4979.5,5020.8
XS Rating Curve= 0 ,0
Exp/Cntr=0.3,0.1

Type RM Length L Ch R = 1 ,88761   ,533,533,533
BEGIN DESCRIPTION:
BIG ELKHART CREEK 88.0
END DESCRIPTION:
XS GIS Cut Line= 3
      3767799.59     10537760.17      3768649.61     10538910.19
      3769249.64     10539360.21
#Sta/Elev= 30
  3551.5  299.15  3567.1  298.08  3759.3  273.83    3937   258.1  4036.9  255.45
  4201.8  255.77  4213.4  252.43  4216.2  251.93  4219.4  252.43  4231.1   255.6
  4251.9  256.21  4331.3  256.39  4345.9  253.32  4387.6   256.4  4402.2  256.19
  4409.5  253.65  4423.1  256.33    4968   258.3  4984.7  258.12  4988.9  255.29
  5009.7  254.01  5024.3  260.09  5045.1  261.08  5095.1  258.08    5218  257.76
  5338.9  258.68  5416.4  262.13  5538.9  276.51  5609.7  288.36  5731.6  301.56
#Mann= 5 ,-1 , 0
  3551.5     .16       0  3567.1     .12       0  4213.4     .07       0
  4219.4     .12       0  5416.4     .16       0
Bank Sta=4968,5045.1
XS Rating Curve= 0 ,0
Exp/Cntr=0.3,0.1

Type RM Length L Ch R = 1 ,88228   ,535,535,535
BEGIN DESCRIPTION:
BIG ELKHART CREEK 87.0
END DESCRIPTION:
XS GIS Cut Line= 3
      3766999.61     10538110.19      3768299.61     10539110.19
      3768699.63     10539910.23
#Sta/Elev= 30
  3387.8  307.26  3392.3  307.28    3449  301.95  3516.1  289.89  3644.2  268.56
  3743.9  258.75  4071.9  252.03  4144.5  254.53  4162.3  251.98    4165  251.48
  4168.3  251.98  4636.5  257.63  4663.6  254.99  4977.5  258.38  5006.2  253.91
  5024.8  259.68  5056.6  260.47  5148.1  263.26  5198.4  261.83  5385.7   266.3
  5461.2  281.23  5475.1  280.68  5483.5  274.74  5489.1  279.97  5497.5  274.93
  5528.2  269.74    5640  269.35  5729.5  282.78  5846.1  293.29  5922.4  301.83
#Mann= 8 ,-1 , 0
  3387.8     .16       0  3392.3     .12       0    3449     .16       0
  3516.1     .12       0  4162.3     .07       0  4168.3     .12       0
  5056.6     .05       0  5846.1     .16       0
#XS Ineff= 1 ,-1
  5461.2  5721.1  281.23
Permanent Ineff=
       F
Bank Sta=4636.5,5148.1
XS Rating Curve= 0 ,0
Exp/Cntr=0.3,0.1

Type RM Length L Ch R = 1 ,87693   ,657,657,657
BEGIN DESCRIPTION:
BIG ELKHART CREEK 86.0
END DESCRIPTION:
XS GIS Cut Line= 3
      3766949.61     10538110.19      3767799.61     10539110.19
      3767649.61      10539910.2
#Sta/Elev= 30
    3682   307.8  3720.3   307.1  3789.9  303.06  3843.5  293.25  3916.5  276.55
  3923.1  277.03  3951.6  267.88  4043.9  256.87    4101  253.34    4235  253.64
  4246.2  250.57    4249  250.07  4252.2  250.57    4257  253.52  4277.8  253.78
  4405.2  254.16  4427.2  251.26  4441.5  254.11  4874.2  256.19  4888.5  254.21
  4980.7  257.08  5004.6  254.13  5014.8  256.98  5025.8  255.06  5136.9  257.44
  5309.8  254.91  5456.5  257.51  5545.7  262.58  5619.3  267.35  5808.4   288.6
#Mann= 7 ,-1 , 0
    3682     .16       0  3720.3     .12       0  3789.9     .16       0
  3843.5     .12       0  4246.2     .07       0  4252.2     .12       0
  5545.7     .05       0
Bank Sta=4980.7,5014.8
XS Rating Curve= 0 ,0
Exp/Cntr=0.3,0.1

Type RM Length L Ch R = 1 ,87036   ,450,450,450
BEGIN DESCRIPTION:
BIG ELKHART CREEK 85.0
END DESCRIPTION:
XS GIS Cut Line= 3
      3766899.61     10538160.18      3767449.61     10539460.19
      3767499.61     10539910.15
#Sta/Elev= 30
  3611.3  306.54  3643.9  304.39  3696.9  295.24  3702.4  296.04  3726.1  289.51
  3731.5  290.48  3741.6  286.48  3817.6     271  3876.4  261.44  3947.9  252.97
  4161.4  253.39  4175.9   250.5  4185.1  252.72  4261.6  254.07  4290.7  253.29
  4296.1     250  4311.4  249.76  4314.1  249.26  4317.4  249.76  4338.1  254.06
  4382.2  252.55  4678.6  255.47  4802.5  253.02  4984.6  254.53  4990.3  251.02
  5008.3  251.66  5013.7  254.13  5153.7  253.34  5263.6  263.09  5475.6  289.08
#Mann= 5 ,-1 , 0
  3611.3     .16       0  3876.4     .12       0  4311.4     .07       0
  4317.4     .12       0  5263.6     .05       0
Bank Sta=4984.6,5013.7
XS Rating Curve= 0 ,0
Exp/Cntr=0.3,0.1

Type RM Length L Ch R = 1 ,86586   ,823,823,823
BEGIN DESCRIPTION:
BIG ELKHART CREEK 84.0
END DESCRIPTION:
XS GIS Cut Line= 4
      3766762.15     10538169.32      3767137.14     10539403.65
      3767173.59     10539773.44      3767506.91     10540315.08
#Sta/Elev= 30
  3518.3  307.94  3591.4  303.54  3655.1  290.92  3667.6  286.19  3733.3   276.8
  3766.2  269.88  3843.2  260.47  3914.2  255.99  4031.3  251.91  4181.6  252.93
  4195.5   249.3  4198.3   248.8  4201.5   249.3  4229.9  253.17  4975.7  253.24
  4988.6  253.13  4995.8  250.18  5015.9  253.35  5146.5  252.93  5267.3  260.14
  5319.1  264.84  5429.2  269.26  5487.2  274.67  5539.3  275.91  5545.2   278.1
  5560.6  276.73  5597.3  279.19  5697.8  289.12  5771.2   288.7  5815.9  291.47
#Mann= 5 ,-1 , 0
  3518.3     .16       0  3914.2     .12       0  4195.5     .07       0
  4201.5     .12       0  5267.3     .05       0
Bank Sta=4975.7,5015.9
XS Rating Curve= 0 ,0
Exp/Cntr=0.3,0.1

Type RM Length L Ch R = 1 ,85763   ,653,653,653
BEGIN DESCRIPTION:
BIG ELKHART CREEK 83.0
END DESCRIPTION:
XS GIS Cut Line= 3
      3766649.61     10538260.16      3766599.61     10539560.19
      3767349.62      10540360.2
#Sta/Elev= 30
  3728.3  306.77  3778.4  305.69  3855.9  298.58  3860.9  299.84  3998.5  277.84
  4092.3  265.47  4116.1  261.74  4121.1  262.48  4128.6  260.57  4208.7  252.56
  4636.5  251.75  4789.1  250.57  4796.1  249.13  4798.9  248.63  4802.1  249.13
  4819.1  251.07  4896.7  251.75  4929.2  249.23  4949.2   251.4  4979.3  251.86
  5009.3  249.15  5026.8  252.19  5078.9   250.8  5566.8  251.05  5675.4  254.08
  5807.6  258.45  5892.6  262.89  6005.5  274.17  6097.8  284.74  6125.9  289.33
#Mann= 5 ,-1 , 0
  3728.3     .16       0  4092.3     .12       0  4796.1     .07       0
  4802.1     .12       0  5675.4     .05       0
Bank Sta=4979.3,5026.8
XS Rating Curve= 0 ,0
Exp/Cntr=0.3,0.1

Type RM Length L Ch R = 1 ,85110   ,407,407,407
BEGIN DESCRIPTION:
BIG ELKHART CREEK 82.0
END DESCRIPTION:
XS GIS Cut Line= 3
      3766499.62     10538260.15      3766083.32     10539655.39
      3766949.61     10540360.19
#Sta/Elev= 30
  3430.8  307.08  3661.9  298.82  3702.2  294.69  3754.3  284.83  3761.3  281.36
  3773.4  280.84  3799.7  277.54    3817  273.29  3832.8   264.5  3858.7  260.21
  3952.6  253.81  4140.5  253.61  4179.9  260.93  4203.1  252.98    4213  252.72
  4218.2  255.47  4251.4  252.62  4307.4  254.62  4361.2  251.69  4986.6  250.38
    4998  246.58  5000.7  246.08    5004  246.58  5023.3  251.14  5477.1  250.64
  5569.8  255.63  5654.7   255.3    5819  258.21  5946.9  267.08  6003.6  273.63
#Mann= 5 ,-1 , 0
  3430.8     .16       0  3773.4     .12       0    4998     .07       0
    5004     .12       0  5654.7     .05       0
Bank Sta=4986.6,5023.3
XS Rating Curve= 0 ,0
Exp/Cntr=0.3,0.1

Type RM Length L Ch R = 1 ,84703   ,444,444,444
BEGIN DESCRIPTION:
Mapping XS ab4668e6
END DESCRIPTION:
XS GIS Cut Line= 5
      3766413.19     10538405.36      3765796.86     10539585.94
      3765874.98     10540063.37      3765440.96     10540879.35
      3764954.84      10541973.1
#Sta/Elev= 30
  3409.7  302.42  3505.4  297.36  3594.3  282.04  3645.4  272.17  3683.9  259.57
  3772.2  254.51  3979.2  253.59  4031.6   260.1  4037.2  255.39  4097.9  252.82
  4125.8  256.84  4158.5   252.6  4816.7  248.57  4918.2  252.81  4979.6  250.57
  4999.1  245.92  5035.9  250.04    5781  252.55  5797.3  249.22    5800  245.56
  5802.7  245.06    5806  245.56  5819.3  251.66  5946.5  251.35  6478.5  252.03
  6667.3  255.98  6765.1  266.36  6971.6   294.4  7107.5  299.03  7346.4  295.84
#Mann= 10 ,-1 , 0
  3409.7     .16       0  3594.3     .12       0    5800     .07       0
    5806     .12       0  5946.5     .05       0  6478.5     .12       0
  6667.3     .16       0  6765.1     .05       0  6971.6     .16       0
  7107.5     .05       0
Bank Sta=4918.2,5035.9
XS Rating Curve= 0 ,0
Exp/Cntr=0.3,0.1

Type RM Length L Ch R = 1 ,84259   ,881,881,881
BEGIN DESCRIPTION:
Mapping XS fd1955f5
END DESCRIPTION:
XS GIS Cut Line= 5
       3766456.6     10538275.15        3765467.     10539681.43
      3765397.55     10540236.99      3765328.11     10540679.69
      3764026.94     10541816.05
#Sta/Elev= 30
    2966  306.53  3068.8   303.3  3161.1  292.52  3175.9     294  3182.1  290.77
  3304.2   273.2  3363.2  261.47    3426  256.25  3836.3  254.33  4317.2  248.68
  4976.6  250.45  5006.8  246.22  5029.7  249.61  5451.1  251.22  5457.1  246.74
  5468.4  245.37  5471.1  244.87  5474.4  245.37  5491.6  251.35  5630.5  251.17
  6145.3  253.22  6154.1  253.35  6415.8  262.01  6450.9  260.84    6487  265.91
    6600   271.4  6701.5   283.8  6708.8  284.59  6854.8  300.05  7421.1  320.92
#Mann= 10 ,-1 , 0
    2966     .16       0  3304.2     .12       0  5468.4     .07       0
  5474.4     .12       0  5630.5     .05       0  6145.3     .12       0
  6154.1     .16       0  6701.5     .05       0  6708.8     .16       0
  6854.8     .05       0
Bank Sta=3836.3,6415.8
XS Rating Curve= 0 ,0
Exp/Cntr=0.3,0.1

Type RM Length L Ch R = 1 ,83378   ,134,134,134
BEGIN DESCRIPTION:
BIG ELKHART CREEK 81.0
END DESCRIPTION:
XS GIS Cut Line= 4
      3766449.61     10538260.19      3764649.61     10540060.19
      3764449.61     10540560.19      3763932.51     10541695.25
#Sta/Elev= 30
    2438  305.84  2565.3  297.64  2799.1  265.92  2862.3  256.54  3017.8  254.77
  3244.1  254.04  3314.8  256.66    3329  253.36  3385.5  252.57  3541.1  254.29
  3625.9  251.47  4205.8   249.3  4234.1   246.8    4333  248.83  4347.2  246.13
  4375.5  248.41  4502.8  246.09  4986.3  248.49  4998.4  243.79  5019.6  243.77
  5022.4  243.27  5025.6  243.77  5037.4  248.62  5103.9  252.63  5306.7  271.67
  5429.2  286.91  5512.7  293.11  5840.8  295.97  6019.3  289.72  6769.4  316.69
#Mann= 5 ,-1 , 0
    2438     .16       0  2799.1     .12       0  5019.6     .07       0
  5025.6     .12       0  5103.9     .05       0
Bank Sta=4986.3,5037.4
XS Rating Curve= 0 ,0
Exp/Cntr=0.3,0.1

Type RM Length L Ch R = 1 ,83244   ,510,510,510
BEGIN DESCRIPTION:
Mapping XS 5d3bbbcf
END DESCRIPTION:
XS GIS Cut Line= 4
      3764783.68     10537784.11      3764892.19     10538652.12
       3764360.5      10540637.8      3763835.52     10541596.36
#Sta/Elev= 30
  2719.5  300.58    2756  297.62  2794.7  294.69  2826.4  291.71  2957.4  290.41
  3043.5   283.7    3144  275.94  3284.7  267.28  3325.8  264.26  3496.2   256.5
  3700.9  251.61  3706.1  247.45  3726.8  251.53  4315.6  248.19    4348  251.38
  4368.7  248.17  4482.6  245.98  4969.1  248.45  4986.8  243.62  4989.6  243.12
  4992.8  243.62  5010.4  248.95  5072.6  248.75  5162.8  257.99  5445.6  289.49
  5528.1  294.23  5857.8  295.87  5992.1  289.22  6079.4  289.24  6742.8  312.59
#Mann= 11 ,-1 , 0
  2719.5     .16       0    2756     .05       0  2794.7     .16       0
  3043.5     .12       0    3144     .16       0  3284.7     .12       0
  3325.8     .16       0  3496.2     .12       0  4986.8     .07       0
  4992.8     .12       0  5162.8     .05       0
Bank Sta=4969.1,5010.4
XS Rating Curve= 0 ,0
Exp/Cntr=0.3,0.1

Type RM Length L Ch R = 1 ,82734   ,775,775,775
BEGIN DESCRIPTION:
BIG ELKHART CREEK 80.0
END DESCRIPTION:
XS GIS Cut Line= 3
       3764649.6      10537960.2      3764049.61     10539960.19
      3763628.79     10541575.53
#Sta/Elev= 30
  2883.9  304.09  3076.2  304.23  3207.5  294.24  3264.2  286.09  3405.9  262.41
  3475.5  256.45  3669.5  247.87  4032.3  246.48  4048.8  249.31  4087.1  245.97
  4491.7  246.77  4512.6  244.56  4543.9  247.27  4731.8  246.28  4752.7  250.67
  4763.1  247.82    4818  246.03  4982.3  247.39  4991.8  243.35  4994.5  242.85
  4997.8  243.35  5013.3  247.33  5137.3  246.48  5244.7  252.87  5465.3  272.53
  5540.3  275.89  5819.3   282.6    5964  280.21  6219.3  296.96  6641.2   311.5
#Mann= 6 ,-1 , 0
  2883.9     .05       0  3264.2     .16       0  3475.5     .12       0
  4991.8     .07       0  4997.8     .12       0  5244.7     .05       0
Bank Sta=4982.3,5013.3
XS Rating Curve= 0 ,0
Exp/Cntr=0.3,0.1

Type RM Length L Ch R = 1 ,81959   ,1377,1377,1377
BEGIN DESCRIPTION:
BIG ELKHART CREEK 79.0
END DESCRIPTION:
XS GIS Cut Line= 3
      3764599.63     10537960.16      3763399.61     10539760.19
      3762699.62     10540360.18
#Sta/Elev= 30
  2853.5  305.99  2969.2  305.98  3077.4  301.63  3258.7  285.35    3418  270.59
  3711.4  246.63  3718.9   244.4  3726.4  247.29  3948.7  245.46  4050.9  247.87
  4086.9  244.58  4432.5  246.28  4540.6     244  4576.7  246.28  4663.8  245.29
  4678.8  248.04  4699.9  244.57  4988.3  246.29  4994.3  242.49  5010.9  242.36
  5013.6  241.86  5016.9  242.36  5020.2  242.36    5024  246.83  5151.3  244.62
  5591.4  244.97  5655.1  248.94  5698.4  254.48  5740.7  257.41  5938.8  287.74
#Mann= 6 ,-1 , 0
  2853.5     .05       0  3258.7     .16       0    3418     .12       0
  5010.9     .07       0  5016.9     .12       0  5698.4     .05       0
Bank Sta=4988.3,5024
XS Rating Curve= 0 ,0
Exp/Cntr=0.3,0.1

Type RM Length L Ch R = 1 ,80582   ,690,690,690
BEGIN DESCRIPTION:
BIG ELKHART CREEK 78.0
END DESCRIPTION:
XS GIS Cut Line= 3
      3763799.62     10537610.18      3762999.61     10538610.19
      3761999.59     10540410.22
#Sta/Elev= 30
  3728.6  289.59    3771  289.27  3835.1  280.16  3863.9  273.34  3899.1  269.65
  3991.9  255.04  4070.4   249.2  4408.5  245.41    4589  244.67  4667.5  242.24
  4995.6  242.94  5014.2  240.54    5017  240.04  5020.2  240.54  5032.1  244.25
  5223.2  241.58  5304.4  243.84  5613.2   243.6  6046.8   247.5  6393.4  256.08
  6579.4  255.47    6724  262.07  6773.9  267.55  6789.2  269.04    6795  271.65
  6805.3  270.74  6832.7  275.29    6909  280.79  6992.6  287.48  7068.4  289.54
#Mann= 8 ,-1 , 0
  3728.6     .16       0  4408.5     .12       0  5014.2     .07       0
  5020.2     .12       0  6579.4     .16       0  6773.9     .05       0
    6909     .16       0  6992.6     .05       0
Bank Sta=4995.6,5032.1
XS Rating Curve= 0 ,0
Exp/Cntr=0.3,0.1

Type RM Length L Ch R = 1 ,79892   ,680,680,680
BEGIN DESCRIPTION:
BIG ELKHART CREEK 77.0
END DESCRIPTION:
XS GIS Cut Line= 3
      3763699.62     10537410.18      3762699.61     10538010.19
      3761299.61     10540010.18
#Sta/Elev= 30
  3833.1  300.04  3926.4  293.38    4043   275.3    4218   253.4  4276.3  248.48
  4454.5  243.03  4633.1  241.42  4964.3  242.28  4986.9  239.98  4988.5  239.79
  4991.3  239.29  4994.5  239.79  5006.7  242.88  5107.8  240.63  5326.7  241.41
  5613.3  242.06  6464.1  247.82  6608.4  251.29  6622.8  249.04  6783.5  256.43
  6787.3  256.71  6837.7  263.77  6871.7  265.32  6959.8  275.12  7037.8  280.36
  7123.7     282    7208  278.05  7334.6  280.93  7365.2  283.04  7440.6  289.07
#Mann= 14 ,-1 , 0
  3833.1     .05       0  4454.5     .12       0  4633.1     .16       0
  4986.9     .12       0  4988.5     .07       0  4994.5     .12       0
  5326.7     .16       0  5613.3     .12       0  6783.5     .16       0
  6787.3     .05       0  6871.7      .1       0    7208     .16       0
  7334.6     .05       0  7365.2     .16       0
Bank Sta=4964.3,5006.7
XS Rating Curve= 0 ,0
Exp/Cntr=0.3,0.1

Type RM Length L Ch R = 1 ,79212   ,737,737,737
BEGIN DESCRIPTION:
BIG ELKHART CREEK 76.0
END DESCRIPTION:
XS GIS Cut Line= 3
      3762199.61     10536810.22      3762099.61     10537810.19
      3761299.62     10539810.17
#Sta/Elev= 30
  4002.6  289.81  4203.6  265.22  4378.4  248.24  4515.1  240.24  4854.3  243.09
  4937.2  239.56  4967.4  241.96  5010.2  239.36  5039.9  241.88  5198.4  239.01
  5201.2  238.51  5204.4  239.01  5326.5  239.74  5444.4  239.88  5675.3  241.72
  5836.9  239.88  5976.9  242.85  6512.2  249.43    6578  250.24    6716  254.25
  6797.4  259.49  6847.9  264.51  6853.3  262.37  6877.6  265.84  6882.9  269.05
  6936.8  275.18  6967.8  275.88  7000.1  282.81  7039.1     286  7161.6  286.14
#Mann= 9 ,-1 , 0
  4002.6     .05       0  4378.4     .12       0  5198.4     .07       0
  5204.4     .12       0  5326.5     .16       0  5444.4     .12       0
  6512.2     .16       0    6578     .05       0  6797.4      .1       0
Bank Sta=4854.3,5976.9
XS Rating Curve= 0 ,0
Exp/Cntr=0.3,0.1

Type RM Length L Ch R = 1 ,78475   ,655,655,655
BEGIN DESCRIPTION:
BIG ELKHART CREEK 75.0
END DESCRIPTION:
XS GIS Cut Line= 3
      3762099.58     10536910.23      3761399.61     10537910.19
      3761199.61     10539910.21
#Sta/Elev= 30
  3777.7  279.29  3886.2  264.55  3907.1  259.79  3928.1  258.93  3993.4  248.65
    4016  247.42  4041.9  244.94  4151.3  241.17  4380.8   239.9  4391.7   239.5
  4517.5  241.31    4605  240.38  4730.4  239.97  5077.5  239.66  5132.4  239.91
  5196.3  238.53  5199.1  238.03  5202.3  238.53  5430.5  240.85  5621.4  239.29
  6112.8  240.64  6194.2  241.62  6274.6  246.22  6357.6  246.65  6449.7  251.88
    6642  268.87  6754.5     279  6887.7  286.21  6960.5  292.24  7008.3  291.11
#Mann= 14 ,-1 , 0
  3777.7     .05       0    4016     .16       0  4041.9     .12       0
  4380.8     .16       0  4391.7     .12       0    4605     .16       0
  4730.4     .12       0  5077.5     .16       0  5132.4     .12       0
  5196.3     .07       0  5202.3     .12       0  6112.8     .16       0
  6449.7     .05       0    6642      .1       0
Bank Sta=4517.5,5430.5
XS Rating Curve= 0 ,0
Exp/Cntr=0.3,0.1

Type RM Length L Ch R = 1 ,77820   ,676,676,676
BEGIN DESCRIPTION:
BIG ELKHART CREEK 74.0
END DESCRIPTION:
XS GIS Cut Line= 3
      3761999.61     10536510.18      3760999.61     10537510.19
      3760399.62     10539110.17
#Sta/Elev= 30
  3565.5  295.39  3692.8  281.71  3961.5  258.89  4167.5  246.68  4274.2  243.68
  4357.5  239.43  4470.6  240.36  4555.5  237.84  4725.2   237.9  4795.9  240.56
  4894.9  237.97  4982.4  239.62  5008.8  237.61  5011.5  237.11  5014.8  237.61
  5025.1  240.15  5110.6  237.85  5397.1  239.81  5587.6  237.67  5678.4  240.09
  5919.6  238.24  5983.6  239.25  6040.3  244.23  6105.6   248.6  6215.9  251.38
  6259.6  256.15  6382.9  263.25  6447.3  266.45    6539  264.01  6688.5  274.46
#Mann= 8 ,-1 , 0
  3565.5     .05       0  4167.5     .16       0  4274.2     .12       0
  5008.8     .07       0  5014.8     .12       0  6040.3     .16       0
  6259.6     .05       0  6382.9      .1       0
Bank Sta=4982.4,5025.1
XS Rating Curve= 0 ,0
Exp/Cntr=0.3,0.1

Type RM Length L Ch R = 1 ,77144   ,728,728,728
BEGIN DESCRIPTION:
BIG ELKHART CREEK 73.0
END DESCRIPTION:
XS GIS Cut Line= 3
      3761599.61     10536010.19      3760599.61     10537010.19
      3760399.61      10538810.2
#Sta/Elev= 30
  3555.7  311.59  3626.4  306.17  3732.5  290.88  3824.4  283.34  3895.1  279.19
  4008.2  264.84  4107.2  256.26  4206.2  249.85  4319.4   245.2  4520.4  240.32
  4657.1  239.61  4704.5  239.67  4790.7  238.89  4827.8  238.78 4899.96  238.57
  4938.6  236.43  4941.4  235.93  4944.6  236.43 5030.16  237.68  5050.4  239.54
  5260.1  237.42    5764  238.17  6219.3  239.54  6348.3  239.27  6452.2  245.69
  6499.3  250.69  6519.4  250.79  6660.3  267.09  6777.2  272.92    6781   272.9
#Mann= 13 ,-1 , 0
  3555.7     .05       0  4520.4     .16       0  4657.1     .12       0
  4704.5     .16       0  4790.7     .05       0  4827.8     .12       0
  4938.6     .07       0  4944.6     .12       0  5260.1     .16       0
    5764     .12       0  6219.3     .16       0  6452.2     .05       0
  6777.2      .1       0
Bank Sta=4899.96,5030.16
XS Rating Curve= 0 ,0
Exp/Cntr=0.3,0.1

Type RM Length L Ch R = 1 ,76416   ,741,741,741
BEGIN DESCRIPTION:
BIG ELKHART CREEK 72.0
END DESCRIPTION:
XS GIS Cut Line= 3
      3760299.61     10535860.19      3760099.61     10536760.19
      3760299.61     10538760.16
#Sta/Elev= 30
  4109.1  281.23  4128.3  280.18  4133.4  281.84  4170.6  278.59  4182.1  279.86
  4225.6  277.05  4269.2  270.48  4274.3   271.4  4317.8     266  4366.5  258.61
  4395.9  251.97  4453.5  246.64  4580.3  240.91  4815.6  238.05  4888.1  237.32
  5006.7  236.39  5008.8  235.98  5011.6  235.48  5014.8  235.98  5020.8  237.26
  5403.7  237.96  5573.7  236.64  6000.4  240.34  6277.2  242.65  6563.2  241.51
  6618.9  241.97  6686.8  247.25  6722.2  247.51  6960.6  270.94    7041  271.56
#Mann= 9 ,-1 , 0
  4109.1     .05       0  4815.6     .07       0  4888.1     .12       0
  5008.8     .07       0  5014.8     .12       0  5403.7     .16       0
  6000.4     .12       0  6563.2     .16       0  6722.2     .05       0
Bank Sta=5006.7,5020.8
XS Rating Curve= 0 ,0
Exp/Cntr=0.3,0.1

Type RM Length L Ch R = 1 ,75675   ,687,687,687
BEGIN DESCRIPTION:
BIG ELKHART CREEK 71.0
END DESCRIPTION:
XS GIS Cut Line= 3
       3760249.6      10535910.2      3759649.61     10536310.19
       3759049.6     10539010.23
#Sta/Elev= 30
  4294.1  280.56  4322.6  278.73  4402.3  263.81  4510.4  249.19  4631.8   240.7
  4740.3  238.64  4776.3  236.29  4884.5  235.19    5302  237.47  5514.2  235.01
  5516.9  234.51  5520.2  235.01  5549.2  237.64  5629.8  235.26  5636.2  236.74
  5906.4   235.8  6651.6   239.6  6839.9  240.89  6913.6  240.86  7084.5  244.95
  7236.9  259.09  7320.1   269.5  7393.1  275.21  7431.5  277.17  7436.6  273.87
  7473.7  273.81  7494.2  274.83  7504.5  278.96  7596.7  285.17  7781.1   288.9
#Mann= 7 ,-1 , 0
  4294.1     .05       0  4631.8     .12       0  5514.2     .07       0
  5520.2     .12       0  6651.6     .05       0  6913.6     .16       0
  7236.9     .05       0
Bank Sta=4740.3,6839.9
XS Rating Curve= 0 ,0
Exp/Cntr=0.3,0.1

Type RM Length L Ch R = 1 ,74988   ,1295,1295,1295
BEGIN DESCRIPTION:
BIG ELKHART CREEK 70.0
END DESCRIPTION:
XS GIS Cut Line= 3
      3759899.64     10535560.17      3759299.61     10535860.19
      3757654.79     10538713.73
#Sta/Elev= 30
  4342.6  281.29    4379  280.59  4454.4  272.32  4588.6  250.75  4626.9  246.56
  4775.9  234.76  4786.8  233.95  4789.6  233.45  4792.8  233.95  4803.8  235.42
  4915.6  236.54  5005.1  234.11  5010.7  236.13  5562.9  234.23  5649.1   235.8
  5782.7  234.74  5804.3  236.33  5825.8  234.68  6045.6  234.94  6120.3  236.84
  6506.7   236.4  6681.3   241.2  6737.2  242.11  6881.6  244.02  7137.2   251.1
    7429  266.99  7701.9  277.21  7905.9  280.17  8088.3  286.69  8307.1  288.04
#Mann= 6 ,-1 , 0
  4342.6     .05       0  4626.9     .12       0  4786.8     .07       0
  4792.8     .12       0  6681.3     .16       0  6737.2     .05       0
Bank Sta=4775.9,5804.3
XS Rating Curve= 0 ,0
Exp/Cntr=0.3,0.1

Type RM Length L Ch R = 1 ,73693   ,918,918,918
BEGIN DESCRIPTION:
BIG ELKHART CREEK 69.0
END DESCRIPTION:
XS GIS Cut Line= 3
      3760052.77     10535046.22      3758978.56     10535306.63
      3756526.29     10537899.96
#Sta/Elev= 30
  3580.2  292.92  3820.1  289.63  3984.7  284.08  4221.4  252.83  4363.7  243.46
  4478.7  234.53  4920.8  235.75  4991.6  232.37  5097.6  234.77  5186.4  232.19
  5189.2  231.69  5192.4  232.19  5394.6  232.71  5451.2  236.41  5550.3  237.15
    5628  233.06  5755.4  236.99  6294.5  235.96  6428.8  242.03  6575.9  253.67
  6611.4  254.32  6689.1  263.17  6738.8   262.8  6745.7  267.46  6897.9  274.08
  7191.5  276.99  7431.8  287.47  7692.6  286.17  7783.3     287  8254.7  286.98
#Mann= 9 ,-1 , 0
  3580.2     .05       0  4363.7     .12       0  5186.4     .07       0
  5192.4     .12       0  6294.5     .16       0  6428.8     .05       0
  6897.9     .16       0  7692.6     .05       0  7783.3     .16       0
Bank Sta=4920.8,5451.2
XS Rating Curve= 0 ,0
Exp/Cntr=0.3,0.1

Type RM Length L Ch R = 1 ,72775   ,1273,1273,1273
BEGIN DESCRIPTION:
BIG ELKHART CREEK 68.0
END DESCRIPTION:
XS GIS Cut Line= 4
      3760117.92      10534807.5      3758490.28     10535013.66
      3757784.98     10535404.29      3756602.29     10536966.75
#Sta/Elev= 30
    2860  279.47  3130.5  288.12  3221.2  285.24  3432.9  287.42  3473.2  286.29
  3558.3  280.75  3735.3  256.81    3836  246.07    3930  238.91  4017.5  234.05
    4461  232.45    4993  233.52    5012  231.59  5014.7  231.09    5018  231.59
  5036.7  234.02  5123.7  233.63  5218.2  237.51  5695.9  243.87  5700.5  243.88
  5902.2  249.91  6032.3  259.29  6230.1  278.83  6285.7  282.24  6292.6  284.24
  6321.1  282.57  6364.7  285.17    7093  284.81  7138.8     282  7266.5  281.44
#Mann= 11 ,-1 , 0
    2860     .05       0    3930     .12       0    5012     .07       0
    5018     .12       0  5218.2     .16       0  5695.9     .12       0
  5700.5     .16       0  5902.2     .05       0  6032.3     .16       0
  6230.1     .05       0  7138.8     .16       0
Bank Sta=4993,5036.7
XS Rating Curve= 0 ,0
Exp/Cntr=0.3,0.1

Type RM Length L Ch R = 1 ,71502   ,533,533,533
BEGIN DESCRIPTION:
BIG ELKHART CREEK 67.0
END DESCRIPTION:
XS GIS Cut Line= 3
      3759195.56     10533364.37      3757600.52      10534829.2
       3756591.4     10536521.92
#Sta/Elev= 30
  3055.8   292.6  3240.8  289.71  3510.2  269.84  3545.4  269.85  3630.5     263
  3722.3  261.55  4104.6  239.53  4352.5  234.36  4585.6  232.85    4961  233.65
  4989.4  231.84  5000.6  230.79  5003.3  230.29  5006.6  230.79  5024.5  232.71
  5362.3  232.05  5464.3  235.85  5635.4  236.07  5836.1  242.28  5927.5   249.3
  6106.6  263.48  6133.9  268.24    6165  269.15  6177.2  272.32  6200.5  272.87
  6213.7  275.61  6367.5  279.23  6404.5  277.52  6505.7  283.19  7192.1  283.66
#Mann= 6 ,-1 , 0
  3055.8     .05       0  4585.6     .12       0  5000.6     .07       0
  5006.6     .12       0  5635.4     .16       0  5927.5     .05       0
Bank Sta=4989.4,5024.5
XS Rating Curve= 0 ,0
Exp/Cntr=0.3,0.1

Type RM Length L Ch R = 1 ,70969   ,875,875,875
BEGIN DESCRIPTION:
BIG ELKHART CREEK 66.0
END DESCRIPTION:
XS GIS Cut Line= 4
      3759249.85     10532615.63      3757709.03     10534113.06
      3757144.79     10534916.01      3756559.73     10536096.97
#Sta/Elev= 30
  2280.7  295.77  2467.9  291.91  2623.6  278.28    2864  263.59    2871  265.06
  2878.2  262.45  2899.3  264.52  2906.5  261.55  2920.6  260.72  2927.6  260.86
  2934.8  264.94  2948.9  265.43  3069.1  263.96  3337.8  250.92    3359  247.32
  3415.6  249.33  3790.3  236.06  4029.3  232.65  4829.1  231.09    4979  232.83
  4984.7  229.94  4987.5  229.44  4990.7  229.94  5014.7  232.52  5389.9  233.39
  5589.8  244.37    5814  264.58  5954.1  280.73  6058.1  283.82  6728.6  282.55
#Mann= 6 ,-1 , 0
  2280.7     .05       0  4029.3     .12       0  4984.7     .07       0
  4990.7     .12       0  5389.9     .16       0  6058.1     .05       0
Bank Sta=4979,5014.7
XS Rating Curve= 0 ,0
Exp/Cntr=0.3,0.1

Type RM Length L Ch R = 1 ,70094   ,1938,1938,1938
BEGIN DESCRIPTION:
BIG ELKHART CREEK 65.0
END DESCRIPTION:
XS GIS Cut Line= 4
      3758457.71     10532832.69      3757133.94     10534134.76
      3757025.43     10534481.98      3755918.75     10535545.26
#Sta/Elev= 30
  2927.4  286.36  2966.8  285.51  3122.2  267.86  3306.2  256.73  3334.4  253.57
  3355.7     258  3405.1  252.28  3412.2     254    3688  234.21  3935.4  230.97
  4345.6  231.58  4363.9  229.18  4366.6  228.68  4369.9  229.18    4579  231.57
  5009.9  229.22  5355.9  239.97  5363.1  237.23  5370.1  239.84  5377.3  235.69
  5426.7  241.95    5564  246.55  5688.3  256.24  5787.4  268.42  5850.9  269.44
  5957.2  279.46  6027.4  282.02  6204.1   282.8  6364.6  283.14  6682.7  282.58
#Mann= 8 ,-1 , 0
  2927.4     .05       0  3306.2     .12       0  4363.9     .07       0
  4369.9     .12       0    5564     .16       0  6027.4     .12       0
  6204.1     .16       0  6364.6     .05       0
Bank Sta=3355.7,5370.1
XS Rating Curve= 0 ,0
Exp/Cntr=0.3,0.1
