--- CEDAR BRANCH.prj (project) ---

Proj Title=CEDAR BRANCH Base Level Engineering
Current Plan=p01
Default Exp/Contr=0.3,0.1
English Units
Geom File=g01
Flow File=f01
Flow File=f02
Plan File=p01
Y Axis Title=Elevation
X Axis Title(PF)=Main Channel Distance
X Axis Title(XS)=Station
BEGIN DESCRIPTION:
CEDAR BRANCH
END DESCRIPTION:
DSS Export Rating Curves= 0
DSS Export Rating Curve Sorted= 0
DSS Export Volume Flow Curves= 0
DXF OffsetX= 0
DXF OffsetY= 0
DXF ScaleX= 1
DXF ScaleY= 10

--- CEDAR BRANCH.p01 (plan) ---

Plan Title=Multiple Run
Short Identifier=Multiple
Geom File=g01
Flow File=f01
Subcritical Flow
K Sum by GR= 0
Std Step Tol= 0.01
Critical Tol= 0.01
Num of Std Step Trials= 20
Max Error Tol= 0.3
Flow Tol Ratio= 0.001
Split Flow NTrial= 30
Split Flow Tol= 0.02
Split Flow Ratio= 0.02
Log Output Level= 0
Friction Slope Method= 1
Unsteady Friction Slope Method= 2
Unsteady Bridges Friction Slope Method= 1
Parabolic Critical Depth
Global Vel Dist=  1 , 1 , 1
Global Log Level= 0
CheckData=True
Encroach Param= -1, 0, 0, 0
BEGIN DESCRIPTION:
Multiple Run
END DESCRIPTION:

--- CEDAR BRANCH.f01 (steady flow) ---

Flow Title=Multiple
Program Version=4.10
Number of Profiles= 7
Profile Names=10-year,25-year,50-year,1pct_min,100-year,1pct_plu,500-year
River Rch & RM=CEDAR BRANCH,Reach-1         ,55411
     947    1318    1633    1485    2009    2716    3052
River Rch & RM=CEDAR BRANCH,Reach-1         ,51132
    1101    1539    1911    1740    2353    3183    3586
River Rch & RM=CEDAR BRANCH,Reach-1         ,46556
    1315    1848    2303    2104    2845    3848    4362
River Rch & RM=CEDAR BRANCH,Reach-1         ,43404
    1545    2183    2730    2501    3382    4574    5215
River Rch & RM=CEDAR BRANCH,Reach-1         ,39182
    1707    2416    3026    2774    3751    5073    5793
River Rch & RM=CEDAR BRANCH,Reach-1         ,34425
    1809    2564    3215    2949    3989    5394    6169
River Rch & RM=CEDAR BRANCH,Reach-1         ,30421
    1936    2739    3427    3137    4243    5738    6532
River Rch & RM=CEDAR BRANCH,Reach-1         ,15874
    2258    3204    4017    3681    4978    6732    7683
Boundary for River Rch & Prof#=CEDAR BRANCH,Reach-1         , 1
Up Type= 0
Dn Type= 3
Dn Slope=0.001
Boundary for River Rch & Prof#=CEDAR BRANCH,Reach-1         , 2
Up Type= 0
Dn Type= 3
Dn Slope=0.001
Boundary for River Rch & Prof#=CEDAR BRANCH,Reach-1         , 3
Up Type= 0
Dn Type= 3
Dn Slope=0.001
Boundary for River Rch & Prof#=CEDAR BRANCH,Reach-1         , 4
Up Type= 0
Dn Type= 3
Dn Slope=0.001
Boundary for River Rch & Prof#=CEDAR BRANCH,Reach-1         , 5
Up Type= 0
Dn Type= 3
Dn Slope=0.001
Boundary for River Rch & Prof#=CEDAR BRANCH,Reach-1         , 6
Up Type= 0
Dn Type= 3
Dn Slope=0.001
Boundary for River Rch & Prof#=CEDAR BRANCH,Reach-1         , 7
Up Type= 0
Dn Type= 3
Dn Slope=0.001
DSS Import GetInterval= 0
DSS Import GetPeak= 0
DSS Import FillOption= 0

--- CEDAR BRANCH.f02 (steady flow) ---

Flow Title=old Multiple
Program Version=4.10
Number of Profiles= 7
Profile Names=10-year,25-year,50-year,1pct_min,100-year,1pct_plu,500-year
River Rch & RM=CEDAR BRANCH,Reach-1         ,39414
     947    1318    1633    1485    2009    2716    3052
River Rch & RM=CEDAR BRANCH,Reach-1         ,35135
    1101    1539    1911    1740    2353    3183    3586
River Rch & RM=CEDAR BRANCH,Reach-1         ,30559
    1315    1848    2303    2104    2845    3848    4362
River Rch & RM=CEDAR BRANCH,Reach-1         ,27407
    1545    2183    2730    2501    3382    4574    5215
River Rch & RM=CEDAR BRANCH,Reach-1         ,23185
    1707    2416    3026    2774    3751    5073    5793
River Rch & RM=CEDAR BRANCH,Reach-1         ,18428
    1809    2564    3215    2949    3989    5394    6169
River Rch & RM=CEDAR BRANCH,Reach-1         ,14424
    1936    2739    3427    3137    4243    5738    6532
River Rch & RM=CEDAR BRANCH,Reach-1         ,135
    2258    3204    4017    3681    4978    6732    7683
Boundary for River Rch & Prof#=CEDAR BRANCH,Reach-1         , 1
Up Type= 0
Dn Type= 1
Dn Known WS=213.52
Boundary for River Rch & Prof#=CEDAR BRANCH,Reach-1         , 2
Up Type= 0
Dn Type= 1
Dn Known WS=214.69
Boundary for River Rch & Prof#=CEDAR BRANCH,Reach-1         , 3
Up Type= 0
Dn Type= 1
Dn Known WS=215.58
Boundary for River Rch & Prof#=CEDAR BRANCH,Reach-1         , 4
Up Type= 0
Dn Type= 1
Dn Known WS=215.24
Boundary for River Rch & Prof#=CEDAR BRANCH,Reach-1         , 5
Up Type= 0
Dn Type= 1
Dn Known WS=216.45
Boundary for River Rch & Prof#=CEDAR BRANCH,Reach-1         , 6
Up Type= 0
Dn Type= 1
Dn Known WS=217.86
Boundary for River Rch & Prof#=CEDAR BRANCH,Reach-1         , 7
Up Type= 0
Dn Type= 1
Dn Known WS=218.53
DSS Import GetInterval= 0
DSS Import GetPeak= 0
DSS Import FillOption= 0

--- CEDAR BRANCH.g01 (geometry) ---

Geom Title=Existing Conditions
Program Version=4.10

River Reach=CEDAR BRANCH    ,Reach-1
Reach XY= 30
      3750449.61     10542560.19      3749399.61     10542410.19
      3749299.61     10541727.59      3747299.61     10541060.19
      3747149.61     10538660.19      3746485.55     10537834.59
       3747865.8     10533387.43      3746149.61     10532810.19
       3746144.5       10528701.      3747072.75       10527870.
        3746741.       10526077.        3747047.       10525365.
        3746485.       10523720.       3747105.5       10522445.
        3746684.       10522083.      3746785.75       10521341.
        3744140.       10519603.      3744205.75       10518875.
      3743330.25       10518060.      3743152.75       10516485.
      3741539.75       10516821.       3741285.5       10514627.
        3740692.       10514040.      3739919.75       10514290.
      3739936.75       10515109.      3739298.25       10515216.
        3739301.       10515650.       3738663.5       10515462.
       3738437.5       10513267.      3737720.91     10512688.74

Type RM Length L Ch R = 1 ,55411   ,1533,1533,1533
BEGIN DESCRIPTION:
CEDAR BRANCH 61.0
END DESCRIPTION:
XS GIS Cut Line= 4
      3751920.62     10542146.09      3750184.52     10542163.45
      3750097.71     10542840.53      3750167.16     10545271.13
#Sta/Elev= 30
  2903.2  283.63  2974.2  283.86  3274.2  280.65  3694.3  279.16  3794.3  277.82
  3824.3   275.8  3884.3   276.3  4154.3  273.79  4174.3  272.27  4204.3  273.33
  4224.3   272.2  4244.3  273.74  4334.3  272.43  4978.9  272.21  5112.8  273.19
    5117  271.95  5119.8  271.45    5123  271.95  5851.9  272.81  6001.9  273.39
    6082  275.16    6132  273.38    6232  274.66  6272.1  273.44  6615.5  274.62
  6832.3  276.92  6892.3  275.94  7292.5  277.57  7562.6  281.54  7753.6  282.88
#Mann= 3 ,-1 , 0
  2903.2     .05       0    5117     .03       0    5123     .05       0
Bank Sta=4154.3,5112.8
XS Rating Curve= 0 ,0
Exp/Cntr=0.3,0.1

Type RM Length L Ch R = 1 ,53878   ,1401,1401,1401
BEGIN DESCRIPTION:
CEDAR BRANCH 60.0
END DESCRIPTION:
XS GIS Cut Line= 3
      3751747.06     10541642.61      3749299.61     10541860.19
      3747299.63     10543860.17
#Sta/Elev= 30
  2542.9  280.55    2711  278.03  2841.5  279.78  3112.6  276.83  3373.6  276.03
  3554.3  272.81  3564.4  271.65  3574.4  273.75  3583.9  273.78  3614.6   272.4
  4337.4  272.02  4457.9   273.2  4487.4  271.84  4489.4  270.59  4492.2  270.09
  4495.4  270.59  4528.1  273.31  4568.3  273.78  4658.7  270.79  4708.9  272.18
  5003.5  271.21    5594  272.23  5608.1   271.2  6697.1  272.41  6725.3  270.83
  6781.9  273.56  6852.6  271.87    7291  273.63  7743.6  273.38  7828.4  275.43
#Mann= 3 ,-1 , 0
  2542.9     .05       0  4489.4     .03       0  4495.4     .05       0
Bank Sta=3554.3,6697.1
XS Rating Curve= 0 ,0
Exp/Cntr=0.3,0.1

Type RM Length L Ch R = 1 ,52477   ,1345,1345,1345
BEGIN DESCRIPTION:
CEDAR BRANCH 59.0
END DESCRIPTION:
XS GIS Cut Line= 3
      3750965.79     10540809.28      3748399.61     10541410.19
      3746399.63     10543210.17
#Sta/Elev= 30
  2364.4  272.75  2388.2  274.59  2452.9  273.14    2987   273.8  3183.5  272.08
  3808.6     272  3849.7  272.79  3890.8  271.59  4541.2  270.37  4917.8  271.26
  5003.4  270.83  5010.8  269.59  5013.6  269.09  5016.8  269.59  5049.7  271.96
  5078.1  270.01  5481.7  271.05  5510.1  269.59  5524.3  270.95  5559.4  271.77
  5616.3  270.37  5686.5  271.06  5955.6  270.58  6267.3  271.63    6749  271.42
  6805.4   272.8  6855.5  271.27  7223.2  274.38  7577.5  274.35  7690.7  275.64
#Mann= 3 ,-1 , 0
  2364.4     .05       0  5010.8     .03       0  5016.8     .05       0
Bank Sta=4917.8,5049.7
XS Rating Curve= 0 ,0
Exp/Cntr=0.3,0.1

Type RM Length L Ch R = 1 ,51132   ,453,453,453
BEGIN DESCRIPTION:
CEDAR BRANCH 58.0
END DESCRIPTION:
XS GIS Cut Line= 3
      3749174.33     10540749.68      3747299.61     10540960.19
      3745499.63     10542960.17
#Sta/Elev= 30
  3113.5  271.89  3168.6  272.85  3349.7  271.28  3812.6  271.46  3822.6  271.39
  4245.3  270.35  5003.4  270.47  5013.8  270.16  5027.8  267.96  5042.2  269.76
  5134.5  270.78    5170  269.98  5198.4   271.6  5226.8  269.61  5269.1  270.79
  5297.1     270  5347.2  270.74  5700.7  270.22  5842.7   271.2  5899.5  270.21
  6238.9  271.45  6253.1  271.55  6621.5   271.5  6685.1  272.63  6706.7  272.55
  6713.5  270.87    6777  272.03  7117.1  271.85  7357.7  274.45  7690.7  275.85
#Mann= 3 ,-1 , 0
  3113.5     .05       0  3822.6     .03       0  6253.1     .05       0
Bank Sta=3812.6,6238.9
XS Rating Curve= 0 ,0
Exp/Cntr=0.3,0.1

Type RM Length L Ch R = 1 ,50679   ,442,442,442
BEGIN DESCRIPTION:
CEDAR BRANCH 57.0
END DESCRIPTION:
XS GIS Cut Line= 3
      3749089.71     10540611.87      3747049.61     10540610.19
      3745249.62     10541010.19
#Sta/Elev= 30
  2959.9  272.04    3810  271.28    4960  270.33  4979.8  267.73    4990   269.6
  5010.2  269.91  5805.4  270.41  5829.8  271.09    5881  269.21  5897.6  269.56
  5911.7  271.35    5922  271.42  5962.9  271.97  5994.9   269.8  6014.1  269.98
  6024.4  271.38  6116.6  270.58  6167.8  271.33  6464.9  271.33  6586.5  273.05
  6598.1  273.01  6608.3  271.34  6618.5   271.2  6628.8  273.55  6649.3  273.24
  6669.8  270.96  6678.7  273.32  6683.8  272.81  6690.2  273.95  6843.9  273.99
#Mann= 3 ,-1 , 0
  2959.9     .05       0    3810     .03       0    5922     .05       0
Bank Sta=3810,5911.7
XS Rating Curve= 0 ,0
Exp/Cntr=0.3,0.1

Type RM Length L Ch R = 1 ,50237   ,450,450,450
BEGIN DESCRIPTION:
CEDAR BRANCH 56.0
END DESCRIPTION:
XS GIS Cut Line= 3
        3749004.     10540414.39      3747149.61     10540210.19
      3745349.58      10540810.2
#Sta/Elev= 30
  3134.4  272.15  3158.9  271.51  3179.1  272.57  3279.7  271.31  3933.6  271.17
  4054.3   270.4  4557.3  270.68  4899.4  269.54  4949.5  269.66  4979.9   270.7
  5002.6  269.76  5010.3  268.23  5021.1  270.05  5105.4  270.79  5263.5  269.88
    6170  270.19  6412.5   271.3  6465.2  270.06  6507.4  272.52    6539  272.54
  6560.1   271.2  6570.6  269.55  6581.1  269.41  6591.7  269.53  6602.2  271.72
  6697.1  270.86  6728.7  272.91  6760.3  270.78  6781.4  273.13  6897.4   273.9
#Mann= 3 , 0 , 0
  3134.4     .05       0  3933.6     .03       0  6412.5     .05       0
Bank Sta=3933.6,6412.5
XS Rating Curve= 0 ,0
Exp/Cntr=0.3,0.1

Type RM Length L Ch R = 1 ,49787   ,500,500,500
BEGIN DESCRIPTION:
CEDAR BRANCH 55.0
END DESCRIPTION:
XS GIS Cut Line= 3
      3748949.63     10539960.19      3747149.61     10539760.19
      3745349.63     10540760.18
#Sta/Elev= 30
  3188.9  271.75  3581.3  271.75  3943.5  270.64  4044.2  271.15  4104.5  270.46
  4315.8  270.39    4346  270.94    4668  269.82  4959.8   269.7  4979.9  270.25
  4989.9  269.89  4997.2  267.53  5013.7  268.47  5022.9  269.87  5094.9  270.28
  5316.9  269.74  5425.6  270.67  6574.1  270.11  6639.3  270.92  6655.3  271.53
  6670.2  270.82  6682.8  269.31  6714.8  272.51  6758.3  273.83  6861.2   273.2
  6866.9  272.84  6876.1   270.5    6883  271.49  6920.7  272.94  7059.1  273.82
#Mann= 3 ,-1 , 0
  3188.9     .05       0    4346     .03       0  6655.3     .05       0
Bank Sta=4346,6639.3
XS Rating Curve= 0 ,0
Exp/Cntr=0.3,0.1

Type RM Length L Ch R = 1 ,49287   ,450,450,450
BEGIN DESCRIPTION:
CEDAR BRANCH 54.0
END DESCRIPTION:
XS GIS Cut Line= 3
      3748949.63     10539460.19      3747149.61     10539260.19
      3745349.57     10540660.22
#Sta/Elev= 30
  3188.9  271.86  4446.6  270.62  4466.7   270.7  4748.5  269.17  4979.9   269.8
  4997.2  267.42  5007.2   269.3  5021.7  269.72  5214.5  270.44  5647.9  269.57
  6460.5  270.47    6475  270.65  6860.5  270.89  6895.8  269.22  6902.1  269.31
  6910.2  271.75  6916.6  270.33  6924.7  272.41  6966.3     273  6974.5  271.62
  6980.8  272.13  7001.6  268.82  7009.8  270.37  7016.1  269.84  7024.3  271.67
  7030.6  270.41  7038.7  272.13  7059.6  272.55  7130.1   271.6  7280.4  273.87
#Mann= 3 ,-1 , 0
  3188.9     .05       0  4446.6     .03       0  6460.5     .05       0
Bank Sta=4466.7,6475
XS Rating Curve= 0 ,0
Exp/Cntr=0.3,0.1

Type RM Length L Ch R = 1 ,48837   ,787,787,787
BEGIN DESCRIPTION:
CEDAR BRANCH 53.0
END DESCRIPTION:
XS GIS Cut Line= 3
      3748949.64      10539410.2      3747149.61     10538810.19
      3745349.62     10540410.18
#Sta/Elev= 30
  3102.6  271.82    3851  270.39  3861.6  270.35  4662.7  269.12  4936.8  269.14
  4968.4  269.88  4997.1  267.22  5007.1   268.9  5013.8  268.36  5049.8  269.75
  6537.4  270.39  6544.1  270.44  6799.1  270.84  6834.3  270.38  6841.8  268.96
  6862.7  268.88  6870.2  271.67  6919.5  271.78  6926.7  271.46  6933.8  269.47
    6948  268.55  6954.7  269.38  6968.9  269.19  6976.4  271.04  6983.1  270.37
  6990.6  271.65    7040   273.1  7096.8  272.74  7259.9  274.75  7408.3  274.21
#Mann= 3 ,-1 , 0
  3102.6     .05       0  3861.6     .03       0  6537.4     .05       0
Bank Sta=3851,6544.1
XS Rating Curve= 0 ,0
Exp/Cntr=0.3,0.1

Type RM Length L Ch R = 1 ,48050   ,1035,1035,1035
BEGIN DESCRIPTION:
CEDAR BRANCH 52.0
END DESCRIPTION:
XS GIS Cut Line= 4
      3748830.32     10539003.71      3747059.52     10538153.03
      3746347.71     10538274.56      3744924.34     10539368.13
#Sta/Elev= 30
  2771.8  271.57  3260.7  270.04  3831.4  270.23  3848.5  270.23  3876.7  269.47
    4482  269.66    4714  268.68  4985.8  269.59  5010.1  267.13  5045.9  269.09
  5415.9  269.09  5460.9  270.37  5481.7  269.76  5496.2  267.63  5504.4  268.68
  5510.7   268.1    5519  270.48  5525.3  268.93  5531.7  270.66  5546.1  270.83
  5575.1  270.41  5582.2  267.83  5595.7  266.49  5604.1  269.26    5654  269.85
  6474.2  270.26  6488.7  270.43  6565.8  271.63  6901.9  272.56  7253.4  272.03
#Mann= 3 ,-1 , 0
  2771.8     .05       0  3831.4     .03       0  6488.7     .05       0
Bank Sta=3848.5,6474.2
XS Rating Curve= 0 ,0
Exp/Cntr=0.3,0.1

Type RM Length L Ch R = 1 ,47015   ,459,459,459
BEGIN DESCRIPTION:
CEDAR BRANCH 51.0
END DESCRIPTION:
XS GIS Cut Line= 4
      3748642.47     10538552.66      3748399.61     10538360.19
      3746599.61     10537360.19      3744799.59      10537960.2
#Sta/Elev= 30
  2648.2   271.5  3090.8  270.29    3172  271.15  3177.7  270.23    3347  269.88
  3670.8  269.72  3701.7  270.74    3736   269.7  3898.4  269.23    4944  269.11
  4949.7   268.3    4960  269.11  4981.7   268.5  5003.2  266.33  5009.2  267.12
  5014.4  270.61  5027.8  271.04  5048.8  270.69  5059.4  267.16    5091  269.21
  5112.1  269.35  5270.2  267.82    5618  269.42    5734   269.2  5755.1  267.96
  5776.2  269.18  6482.4  268.61  6672.1     270  6809.2  272.55  6914.6  272.24
#Mann= 3 ,-1 , 0
  2648.2     .05       0  4949.7     .04       0  5059.4     .05       0
Bank Sta=4944,5027.8
XS Rating Curve= 0 ,0
Exp/Cntr=0.3,0.1

Type RM Length L Ch R = 1 ,46556   ,462,462,462
BEGIN DESCRIPTION:
CEDAR BRANCH 50.0
END DESCRIPTION:
XS GIS Cut Line= 3
      3748749.57     10538560.16      3746749.61     10536960.19
      3744749.58      10537760.2
#Sta/Elev= 30
  2438.8     272  2474.8  271.21    3861  269.01  3911.5  270.37  3961.9  269.34
  4346.1  269.18  4928.8  270.04  4992.8  267.97  5009.2  266.06  5014.8   266.7
  5021.5  269.11  5044.4  270.71  5053.9  270.56  5063.3  268.85  5068.7  269.73
  5075.4  267.49  5092.9  268.97  5098.3  268.27  5129.2  269.38  5409.3  267.52
  5655.6  269.58  5709.5  267.76  5798.4  268.79  5822.6  268.67  5829.3  267.53
  5846.8  268.72  5930.3  269.27  6917.1   268.8  6983.1  270.82  7154.1  271.53
#Mann= 3 ,-1 , 0
  2438.8     .05       0  4928.8     .04       0  5098.3     .05       0
Bank Sta=4928.8,5044.4
XS Rating Curve= 0 ,0
Exp/Cntr=0.3,0.1

Type RM Length L Ch R = 1 ,46094   ,431,431,431
BEGIN DESCRIPTION:
CEDAR BRANCH 49.0
END DESCRIPTION:
XS GIS Cut Line= 3
      3748899.59     10538360.17      3746899.61     10536560.19
      3744708.59     10537437.13
#Sta/Elev= 30
  2309.3  271.38    3010  269.96  3066.8  271.27  3123.6  270.14  3321.7  269.95
  4915.2  269.59  4929.4  269.77  4992.9  269.14  5044.4  266.61  5063.3  270.54
  5086.2  270.22  5092.9     269  5098.3  269.69  5107.7  266.62  5122.5  266.59
  5129.3  268.32  5146.7  269.23  5176.3  269.39  5290.8  268.37  5547.8  269.26
  5700.1  267.56  5732.4  268.33  5768.6  267.53  5775.3  266.06  5798.2  267.74
  5905.9  267.05  5915.6  268.07    6508  267.86  7305.7  269.47    7360  270.15
#Mann= 3 ,-1 , 0
  2309.3     .05       0  4915.2     .04       0  5176.3     .05       0
Bank Sta=4929.4,7305.7
XS Rating Curve= 0 ,0
Exp/Cntr=0.3,0.1

Type RM Length L Ch R = 1 ,45663   ,462,462,462
BEGIN DESCRIPTION:
CEDAR BRANCH 48.0
END DESCRIPTION:
XS GIS Cut Line= 4
      3748799.63     10536360.19      3746999.61     10536160.19
      3745199.61     10537160.19      3744720.57     10537245.46
#Sta/Elev= 30
  3188.9  270.67  3420.3   270.6  3510.9  269.55  3782.6  268.93  4919.5  269.44
  4959.8  269.14  4994.5  266.43  4997.2  265.93  5000.5  266.43  5035.5  269.97
    5111  270.83  5116.7  266.78  5125.8  267.87  5138.4  267.46  5160.2  268.52
  5411.8  268.69  5434.7  269.95  5514.8  268.61  5949.5   267.5  5972.4  266.46
  5983.8  267.35  6109.6  268.42  6132.5  267.69    6200  268.47  6227.5  267.85
    6796  267.88  6839.5  268.75  7051.1  269.37  7343.5  268.77  7545.7  269.99
#Mann= 4 ,-1 , 0
  3188.9     .05       0  4994.5     .04       0  5000.5     .05       0
  7545.7     .05       0
Bank Sta=4919.5,5111
XS Rating Curve= 0 ,0
Exp/Cntr=0.3,0.1

Type RM Length L Ch R = 1 ,45201   ,442,442,442
BEGIN DESCRIPTION:
CEDAR BRANCH 47.0
END DESCRIPTION:
XS GIS Cut Line= 4
      3749149.65      10536360.2      3747149.61     10535760.19
      3745047.34      10536594.7      3743824.02     10537323.49
#Sta/Elev= 30
  2911.9  272.41  2928.5  270.55  3162.5  271.85  4290.9  268.16  4395.3  269.57
  4926.9   268.5  4989.6  268.11    4997  265.76  4999.8  265.26    5003  265.76
  5014.8  267.24  5032.3  266.11  5039.2  268.14  5044.5  267.24  5068.8  269.63
  5107.6  266.99  5152.5  268.81  5608.9  268.38  5716.9  267.64  5741.2  265.76
  5770.9  268.25  5817.7  266.37  5854.6   267.8  5871.5  266.09  5878.9  267.52
  5884.2  266.13  7126.3  268.83  8050.7  268.19  8271.9  270.38  8685.8  270.59
#Mann= 3 ,-1 , 0
  2911.9     .05       0    4997     .04       0    5003     .05       0
Bank Sta=4997,5003
XS Rating Curve= 0 ,0
Exp/Cntr=0.3,0.1

Type RM Length L Ch R = 1 ,44759   ,1355,1355,1355
BEGIN DESCRIPTION:
CEDAR BRANCH 46.0
END DESCRIPTION:
XS GIS Cut Line= 4
      3749049.61     10535360.19      3747249.61     10535360.19
      3745318.17     10536209.28      3743385.84     10536657.21
#Sta/Elev= 30
    3200  271.03    3580  270.31    3660  268.71    3740  270.01    4770  267.63
    4940  268.79    4970  268.19    4997  264.59  4999.8  264.09    5003  264.59
  5032.3  269.03  5054.6  268.76  5061.1  266.29  5066.6  266.28  5084.4  268.26
  5136.6  268.66  6299.5  268.03  6321.8  267.42  6333.8  264.71  6343.6  264.59
  6375.3  267.77  6399.1  267.76  6403.8  267.66  6409.3  265.38  6427.2  265.09
  6441.9  266.81  6540.2  265.94  6867.9  268.37  8648.1  267.48  9093.4  269.75
#Mann= 5 ,-1 , 0
    3200     .05       0    4997     .04       0    5003     .05       0
  6375.3     .08       0  6399.1     .05       0
Bank Sta=4997,5003
XS Rating Curve= 0 ,0
Exp/Cntr=0.3,0.1

Type RM Length L Ch R = 1 ,43404   ,1275,1275,1275
BEGIN DESCRIPTION:
CEDAR BRANCH 45.0
END DESCRIPTION:
XS GIS Cut Line= 4
      3749378.77     10534747.91      3747434.29     10534088.17
      3745266.09     10534964.49      3743334.19     10536073.64
#Sta/Elev= 30
  3148.5  269.63  4858.3  267.95  4942.8   268.9  4974.5  267.14  4991.8  265.24
    4997  263.19  4999.8  262.69    5003  263.19  5006.2  267.07  5023.2   269.3
  5037.8  269.38  5048.4  265.92  5059.9  268.54    5086   268.7  5836.1  266.04
  5943.4  266.98  6727.7  267.42  7213.1   265.2  7234.6  263.19  7256.2  264.82
  7434.9  267.28  8164.6  267.01  8486.8  267.58  8508.5  269.07  8539.6  268.86
  8555.5  267.34  8597.2  268.13  8969.9  267.49  9484.7  269.92  9768.1  268.86
#Mann= 5 ,-1 , 0
  3148.5     .05       0    4997     .04       0    5003     .05       0
  8508.5     .08       0  8555.5     .05       0
Bank Sta=4997,5003
XS Rating Curve= 0 ,0
Exp/Cntr=0.3,0.1

Type RM Length L Ch R = 1 ,42129   ,1507,1507,1507
BEGIN DESCRIPTION:
CEDAR BRANCH 44.0
END DESCRIPTION:
XS GIS Cut Line= 3
       3749673.9     10533168.04      3747903.04     10532994.42
      3745084.49     10534628.65
#Sta/Elev= 30
  2766.2  270.31  3071.9  270.16  3201.4   268.5  3694.9  267.33  4124.8  267.68
  4197.3  266.54  4984.3  266.91  4990.1  263.14  5000.1  263.01  5021.6  265.34
  5027.4  267.77    5035     267  5043.1  268.29  5048.9  268.89  5070.4  266.41
  5809.5  267.17  6226.6   265.9  6301.1  263.59  6526.4  266.19  7135.9  266.36
  7216.2   265.4  7237.8  264.42  7243.6  262.33  7256.3  261.64  7259.1  261.14
  7262.3  261.64  7280.8  263.75  7398.4  263.42  7537.6  266.42  7803.6  267.04
#Mann= 5 ,-1 , 0
  2766.2     .09       0  4990.1     .07       0  5043.1     .05       0
  7256.3     .07       0  7262.3     .05       0
Bank Sta=4984.3,5048.9
XS Rating Curve= 0 ,0
Exp/Cntr=0.3,0.1

Type RM Length L Ch R = 1 ,40622   ,1440,1440,1440
BEGIN DESCRIPTION:
CEDAR BRANCH 42.0
END DESCRIPTION:
XS GIS Cut Line= 3
      3747999.64     10531960.18      3746199.61     10532760.19
      3744399.62     10534360.18
#Sta/Elev= 30
  3030.2  267.49    3840  261.97  3872.9  264.07    3983  264.67  4640.4  264.12
  4718.9  262.77  4835.2  260.34  4901.5  261.85  4939.1  259.09  4962.4  261.18
  4985.6  259.17  4997.3  261.03    5047  261.17  5078.2  261.15  5092.4  258.87
  5121.5  260.45    5411  263.82  5708.7  259.09  5764.7  260.12  5775.9  258.07
  5778.7  257.57  5781.9  258.07  5800.7  260.53  5878.5  259.49    5942  262.07
    6289  262.99  6480.5  260.79    6509  262.46  6664.5  265.81  7408.3  267.47
#Mann= 6 ,-1 , 0
  3030.2     .16       0  4640.4     .12       0    5047     .16       0
  5121.5     .05       0  5775.9     .07       0  5781.9     .05       0
Bank Sta=4718.9,6509
XS Rating Curve= 0 ,0
Exp/Cntr=0.3,0.1

Type RM Length L Ch R = 1 ,39182   ,815,815,815
BEGIN DESCRIPTION:
CEDAR BRANCH 41.0
END DESCRIPTION:
XS GIS Cut Line= 3
      3748849.61     10531760.19      3746149.61     10531760.19
      3743749.59      10534460.2
#Sta/Elev= 30
    2300  267.42  2329.6  267.11    2460  267.73  2527.4  266.31    3280  267.18
    3300     266    3460   265.6    3490   266.9  3713.9  265.49    3741  266.13
  4236.3  265.06    4390  264.99  4518.8  261.21    4570  261.44    4740  257.35
  4803.2  257.54    4940  257.19    4957  255.08  4959.7  254.58    4963  255.08
    4970  257.44  5019.3  258.47  5184.4  261.68  5523.9  265.37  5897.1   265.7
  6048.7  265.27  6374.3  266.42  7599.4  264.88  8321.9  269.26  8612.5  269.25
#Mann= 13 ,-1 , 0
    2300     .12       0  2329.6     .07       0  2527.4     .16       0
  3713.9     .05       0    3741     .16       0  4236.3     .05       0
  4518.8     .16       0  4803.2     .12       0    4957     .07       0
    4963     .12       0  5019.3     .05       0  5897.1     .16       0
  6048.7     .05       0
Bank Sta=4570,5184.4
XS Rating Curve= 0 ,0
Exp/Cntr=0.3,0.1

Type RM Length L Ch R = 1 ,38367   ,549,549,549
BEGIN DESCRIPTION:
CEDAR BRANCH 40.0
END DESCRIPTION:
XS GIS Cut Line= 3
      3748749.58     10531060.19      3746064.97     10531139.55
      3743949.64     10533760.15
#Sta/Elev= 30
  2336.4  267.32    2437  267.63    2536  267.08  2734.1  266.59    3184  266.21
  3790.3  265.49  4169.4  264.68  4262.7  265.12  4597.4  261.89    4811  256.57
  4987.5  255.86  4997.1  253.31  5004.5  251.03  5007.3  250.53  5010.5  251.03
  5017.4  255.11  5034.1  252.56  5040.5  255.92  5054.9  256.46  5061.6  253.61
  5075.7  256.54  5254.3  261.28  6374.7  265.71  6464.9  265.37  6700.3  265.62
  7002.7  268.05  7074.7  264.74  7309.7  264.75  7664.8  267.97    8390  268.88
#Mann= 15 ,-1 , 0
  2336.4     .16       0    2437     .05       0    2536     .16       0
  2734.1     .05       0    3184     .16       0  3790.3     .05       0
  4169.4     .16       0  4262.7     .05       0    4811     .12       0
  4997.1     .05       0  5004.5     .03       0  5010.5     .05       0
  6374.7     .07       0  6464.9     .16       0  6700.3     .05       0
Bank Sta=4597.4,5254.3
XS Rating Curve= 0 ,0
Exp/Cntr=0.3,0.1

Type RM Length L Ch R = 1 ,37818   ,1415,1415,1415
BEGIN DESCRIPTION:
CEDAR BRANCH 39.0
END DESCRIPTION:
XS GIS Cut Line= 3
      3748749.58     10530460.19      3746083.39     10530906.12
      3743349.58      10531960.2
#Sta/Elev= 30
  2391.3  268.01  2796.8  265.28  3517.2  266.68  3557.2  265.11  3567.4  267.26
  3587.7  265.23  3658.6  266.83  3964.3  265.89    4133  265.48  4708.9  264.84
  4865.2  260.06  4927.5  256.12  4986.8  254.98  5004.1  252.46  5006.9  251.96
  5010.1  252.46  5025.3  255.03  5138.9  255.49  5334.4  260.47  5653.2   263.5
  6042.8  263.78  6429.5  267.27  6628.1  266.76    6707  266.82  7278.2  266.64
  7338.3  268.48  7552.9  265.25  7911.9  266.48  8009.5  269.27  8024.5  267.23
#Mann= 14 ,-1 , 0
  2391.3     .16       0  3964.3     .05       0    4133     .16       0
  4708.9     .05       0  4927.5     .16       0  5004.1     .07       0
  5010.1     .16       0  5138.9     .05       0  5653.2     .16       0
  6042.8     .05       0  6628.1     .08       0    6707     .05       0
  7278.2     .12       0  7911.9     .05       0
Bank Sta=4865.2,5334.4
XS Rating Curve= 0 ,0
Exp/Cntr=0.3,0.1

Type RM Length L Ch R = 1 ,36403   ,182,182,182
BEGIN DESCRIPTION:
CEDAR BRANCH 38.0
END DESCRIPTION:
XS GIS Cut Line= 6
      3748131.25     10529966.69      3746992.39     10529883.36
        3746416.     10530091.69      3745964.61     10530154.19
      3745193.78     10530536.13      3744888.24     10531188.89
#Sta/Elev= 30
  3037.1  266.68  3048.1  266.85  3128.5   265.3    3547  264.32  3905.2     264
  4262.8  264.53  4369.4  264.75  4431.3  264.78    4476  265.37  4629.8   264.7
  4689.3  262.27  4692.1  262.15  4838.4   257.2  4978.7  252.64  4994.3  248.99
  4995.7  248.53  4998.5  248.03  5001.7  248.53  5003.8   250.8  5018.7  253.11
  5058.8  251.98    5201  255.31  5225.9  257.48    5385  262.32  5497.4  262.11
  5974.9  263.64  6036.6  265.23  6554.4  263.52  6702.4  266.39  6831.7  266.05
#Mann= 17 ,-1 , 0
  3037.1     .16       0  3048.1     .12       0  3128.5     .16       0
    3547     .05       0  3905.2     .16       0  4262.8      .1       0
  4369.4     .05       0  4431.3     .16       0    4476     .05       0
  4689.3     .08       0  4692.1     .05       0  4994.3     .16       0
  4995.7     .07       0  5001.7     .16       0    5201     .05       0
    5385     .16       0  5497.4     .05       0
Bank Sta=4838.4,5225.9
XS Rating Curve= 0 ,0
Exp/Cntr=0.3,0.1

Type RM Length L Ch R = 1 ,36221   ,1083,1083,1083
BEGIN DESCRIPTION:
CEDAR BRANCH 37.0
END DESCRIPTION:
XS GIS Cut Line= 6
      3747832.66     10529605.58      3747061.83     10529681.97
      3746409.06     10529918.08        3746166.     10529945.86
        3745416.     10529911.13      3744235.42     10530334.76
#Sta/Elev= 30
  3371.5  264.54  3636.8  263.92  3957.4  261.91  4138.3  265.04  4169.7  263.28
  4403.1  263.76  4419.1   263.7  4509.7  264.44  4679.8   261.9    4723  261.56
  4777.1  257.05  4916.9  254.69  4988.3  252.05  4997.8  246.18  5000.5  245.68
  5003.8  246.18  5020.9  251.83  5077.6  250.45  5097.8  253.52  5181.4  256.91
  5375.5  260.02  5572.3  263.05  5952.9  264.31  6084.7  263.99  6223.8  264.34
  6417.5  264.04  6459.2  264.24  6565.7  264.47  6954.4  264.97    7090  266.46
#Mann= 19 ,-1 , 0
  3371.5     .16       0  3636.8     .05       0  4403.1     .16       0
  4419.1     .08       0  4509.7     .05       0  4679.8     .08       0
    4723     .05       0  4916.9     .16       0  4997.8     .07       0
  5003.8     .16       0  5375.5     .12       0  5572.3     .16       0
  5952.9     .12       0  6084.7     .16       0  6223.8     .12       0
  6417.5     .16       0  6459.2     .12       0  6565.7     .16       0
  6954.4     .05       0
Bank Sta=4777.1,5181.4
XS Rating Curve= 0 ,0
Exp/Cntr=0.3,0.1

Type RM Length L Ch R = 1 ,35139   ,713,713,713
BEGIN DESCRIPTION:
CEDAR BRANCH 35.0
END DESCRIPTION:
XS GIS Cut Line= 3
      3748111.76     10529227.54      3746017.56     10529053.93
      3744553.63     10529682.88
#Sta/Elev= 30
    3078   268.1  3220.6  267.53  3260.8  265.39  3371.1   266.8    3952  264.26
  4030.2  264.19  4284.3  262.87  4394.6   264.8  4498.5  262.91  4725.8  259.29
  4799.5  254.98  4806.1  255.21  4976.6  248.59  4983.7  243.38  4986.4  242.88
  4989.7  243.38    4990  243.42  5006.7  249.18  5026.8  250.21  5296.9  255.39
  5433.5  260.79  5978.3  264.19  6156.7  266.67  6254.7  264.32  6309.1  266.82
  6461.9     266    6517  266.02  6559.4  267.84    6699  265.28  6772.7  266.38
#Mann= 12 ,-1 , 0
    3078     .05       0    3952     .16       0  4030.2     .05       0
  4498.5     .16       0  4799.5     .12       0  4983.7     .07       0
  4989.7     .12       0    4990     .16       0  5433.5     .05       0
  5978.3     .16       0  6461.9     .12       0    6517     .16       0
Bank Sta=4806.1,5296.9
XS Rating Curve= 0 ,0
Exp/Cntr=0.3,0.1

Type RM Length L Ch R = 1 ,34425   ,1597,1597,1597
BEGIN DESCRIPTION:
CEDAR BRANCH 34.0
END DESCRIPTION:
XS GIS Cut Line= 2
      3747312.79     10528914.57      3745819.74     10528341.66
#Sta/Elev= 30
  4060.9  265.95  4258.5  262.87  4399.8  262.68  4441.8   263.4  4537.3  262.93
  4650.5  259.18  4679.5  257.87  4754.9  254.83  4786.1  253.83  4870.8  251.85
  4910.5  248.55  4920.2  251.08  4925.5  248.35  4950.2  252.16  4955.5  250.56
  4980.2  249.77  4996.2  243.02  5001.9  242.91  5004.6  242.41  5007.9  242.91
  5010.2  247.67  5017.6  248.86  5110.2  247.86  5135.4  250.11  5253.2  254.22
  5338.4  258.86  5368.4  262.65  5398.2  262.81  5507.8  264.78  5660.1  264.42
#Mann= 10 ,-1 , 0
  4060.9     .05       0  4399.8     .16       0  4441.8     .05       0
  4650.5     .16       0  4679.5     .05       0  4754.9     .12       0
  5001.9     .07       0  5007.9     .12       0  5110.2     .16       0
  5398.2     .05       0
Bank Sta=4786.1,5253.2
XS Rating Curve= 0 ,0
Exp/Cntr=0.3,0.1

Type RM Length L Ch R = 1 ,32828   ,351,351,351
BEGIN DESCRIPTION:
CEDAR BRANCH 33.0
END DESCRIPTION:
XS GIS Cut Line= 3
      3748076.68     10527629.84       3747295.4     10527490.95
      3745628.73     10527907.62
#Sta/Elev= 30
  3851.2  264.62  4071.7  263.85  4329.5  260.67  4337.5  260.49  4354.4  260.37
  4563.8  255.38  4681.6  250.81  4787.9  247.44  4911.6  246.33  4939.3   244.2
  4970.2  245.84    4994  244.29  4998.2  239.53  5000.9  239.03  5004.2  239.53
  5011.5  246.62  5117.7  249.74  5135.2  251.64  5178.3  252.38  5241.4   254.7
  5318.7  253.47  5442.4  256.89  5447.6  255.77  5483.7  256.69  5506.2  255.44
  5547.5  257.95  5743.3  262.37  5918.6   264.2  6114.4  264.34  6362.7  262.18
#Mann= 7 ,-1 , 0
  3851.2     .05       0  4329.5     .16       0  4337.5     .05       0
  4354.4     .16       0  4998.2     .07       0  5004.2     .16       0
  5178.3     .05       0
Bank Sta=4681.6,5135.2
XS Rating Curve= 0 ,0
Exp/Cntr=0.3,0.1

Type RM Length L Ch R = 1 ,32477   ,907,907,907
BEGIN DESCRIPTION:
CEDAR BRANCH 32.0
END DESCRIPTION:
XS GIS Cut Line= 3
      3747799.56     10527210.19      3746989.84     10527213.17
      3745999.65     10527510.18
#Sta/Elev= 30
  4074.9  262.77  4122.7  261.87  4194.9  260.24  4374.9  260.99  4514.9  256.23
  4574.9  252.33  4624.9  250.54  4644.9  251.12  4654.9  248.95  4674.9  247.83
  4890.9  244.51  4968.4  245.51  4978.8  242.53  4986.3  237.67    4989  237.17
  4992.3  237.67  4995.3  239.94  5000.5  239.57  5010.1  247.38  5028.3  252.03
  5033.6  250.16  5051.9  252.95  5106.1   254.4  5260.7  255.21  5308.5  257.19
  5379.9  255.87  5490.4  257.01  5731.4  261.38  5759.2  262.89  5918.4  264.13
#Mann= 5 ,-1 , 0
  4074.9     .05       0  4122.7     .16       0  4986.3     .07       0
  4992.3     .16       0  5106.1     .05       0
Bank Sta=4644.9,5028.3
XS Rating Curve= 0 ,0
Exp/Cntr=0.3,0.1

Type RM Length L Ch R = 1 ,31570   ,288,288,288
BEGIN DESCRIPTION:
CEDAR BRANCH 31.0
END DESCRIPTION:
XS GIS Cut Line= 3
       3748649.6     10527360.18      3746864.84     10526615.95
      3745684.48     10527164.47
#Sta/Elev= 30
  3088.1  266.26  3147.7  265.76  3253.2  264.97  3358.6  264.84  3386.5  263.17
  3391.9   265.1  3410.3   262.5  3555.3  262.73  3747.1  264.06  4014.8  261.21
  4204.1  255.34  4343.9  257.69  4479.2  256.16  4756.6  247.72  4786.8  242.97
  4792.2  246.48    4800  243.07  4832.5  243.84  4845.3  239.89  4863.7  244.46
  4984.1  243.39  5002.8  237.68  5005.6  237.18  5008.8  237.68  5027.6  243.53
  5165.8  247.49  5186.8  247.95  5444.1  257.58  5810.5  264.33  6323.4  264.31
#Mann= 9 ,-1 , 0
  3088.1     .05       0  3147.7     .08       0  3253.2     .05       0
  3358.6     .08       0  3555.3     .05       0  4014.8     .16       0
  5002.8     .07       0  5008.8     .16       0  5165.8     .05       0
Bank Sta=4756.6,5186.8
XS Rating Curve= 0 ,0
Exp/Cntr=0.3,0.1

Type RM Length L Ch R = 1 ,31282   ,720,720,720
BEGIN DESCRIPTION:
CEDAR BRANCH 30.0
END DESCRIPTION:
XS GIS Cut Line= 3
      3747899.61     10526210.19      3746799.61     10526410.19
      3745999.57      10526610.2
#Sta/Elev= 30
  3913.5  263.51  3990.9  263.16  4050.4  261.69  4269.2  257.88  4392.5  258.31
  4499.2  254.38    4564  254.13  4746.9  247.19  4797.8  246.96  4921.7  243.12
  4951.5  243.42  4980.7  241.49  4987.9  235.73  4990.6  235.23  4993.9  235.73
  4999.8  236.52  5011.2   242.7  5041.8  242.74  5054.7  240.42  5062.5  240.94
  5072.8  244.56  5090.8  246.72    5132  249.26  5144.9  248.37  5227.4  250.34
  5268.6  253.78  5289.2  252.88  5338.2  257.26  5390.2  257.56  5856.2  263.41
#Mann= 7 ,-1 , 0
  3913.5     .05       0  3990.9     .16       0  4050.4     .05       0
  4921.7     .16       0  4987.9     .07       0  4993.9     .16       0
  5390.2     .05       0
Bank Sta=4797.8,5090.8
XS Rating Curve= 0 ,0
Exp/Cntr=0.3,0.1

Type RM Length L Ch R = 1 ,30562   ,141,141,141
BEGIN DESCRIPTION:
CEDAR BRANCH 28.0
END DESCRIPTION:
XS GIS Cut Line= 5
      3747287.09     10526167.64      3747026.68      10526011.4
      3746867.82     10525948.03       3746808.8     10525901.15
      3746147.31     10525944.56
#Sta/Elev= 30
  4560.6  257.77  4665.5  255.71  4776.3  248.45  4893.4  243.63  4941.6  242.31
  4968.8  241.73  4979.6  239.11    4987  239.35  4998.1  235.05  5000.8  234.55
  5004.1  235.05  5011.2  239.51  5016.6  240.49  5039.6  241.17  5054.1  235.78
  5060.5  237.54  5068.5  236.84  5074.5  240.58  5112.8  242.08    5139  239.02
    5150  239.36    5160  242.01    5190   243.8  5210.1  244.32  5230.1  246.35
  5240.2  249.31  5265.1  251.25  5320.2   253.4  5520.8  254.23  5773.6  258.25
#Mann= 7 ,-1 , 0
  4560.6     .05       0  4941.6     .16       0  4998.1     .07       0
  5004.1     .16       0  5074.5     .05       0    5139     .16       0
  5265.1     .05       0
Bank Sta=4893.4,5190
XS Rating Curve= 0 ,0
Exp/Cntr=0.3,0.1

Type RM Length L Ch R = 1 ,30421   ,1261,1261,1261
BEGIN DESCRIPTION:
CEDAR BRANCH 27.0
END DESCRIPTION:
XS GIS Cut Line= 5
       3747376.5     10526126.84      3747133.45     10525927.19
      3746881.71     10525819.55      3746631.71     10525727.54
      3746249.76     10525602.54
#Sta/Elev= 30
  4472.6  260.24  4631.5  256.25  4660.2  256.68  4681.1  253.85  4773.6  248.21
  4870.7  243.92  4888.9  244.44  4923.3  240.84  4932.7  242.38  4941.5  241.74
  4965.1  235.87  4970.5  237.58  4987.1  234.87  5005.8  234.11  5008.6  233.61
  5011.8  234.11  5041.3  236.16  5046.7  241.43  5064.7  239.45  5076.3  242.57
  5106.8  242.91  5116.4   244.3  5126.6  246.98  5148.4  244.23  5169.7   244.6
  5334.8   251.7  5382.1  250.08  5483.6  250.64  5586.4  251.27  5729.2  253.77
#Mann= 5 ,-1 , 0
  4472.6     .05       0  5005.8     .04       0  5011.8     .05       0
  5483.6     .08       0  5586.4     .05       0
Bank Sta=4888.9,5116.4
XS Rating Curve= 0 ,0
Exp/Cntr=0.3,0.1

Type RM Length L Ch R = 1 ,29161   ,417,417,417
BEGIN DESCRIPTION:
CEDAR BRANCH 26.0
END DESCRIPTION:
XS GIS Cut Line= 3
      3747349.57     10525060.19      3746799.61     10525060.19
      3745999.58     10525560.21
#Sta/Elev= 30
  4485.4  259.33  4582.3  255.16  4833.7  244.21  4895.4  242.42  4975.4  237.75
  4992.4  230.45  4995.1  229.95  4998.4  230.45  5005.4  235.12  5025.4  238.19
  5064.3  238.71  5106.7  237.07    5122  238.52  5137.4  237.35  5195.1  239.78
    5201  237.94  5231.7  238.67  5259.4  243.41  5269.5   245.4  5274.2  246.92
  5295.4  247.71    5326  244.37  5331.9  245.44  5383.8  244.22  5551.3  251.52
  5587.8  251.22  5609.1  253.58  5724.6  254.55  5934.5  259.36  5978.8  257.48
#Mann= 6 ,-1 , 0
  4485.4     .16       0  4582.3     .05       0  4833.7     .16       0
  4992.4     .07       0  4998.4     .16       0  5269.5     .05       0
Bank Sta=4895.4,5259.4
XS Rating Curve= 0 ,0
Exp/Cntr=0.3,0.1

Type RM Length L Ch R = 1 ,28743   ,515,515,515
BEGIN DESCRIPTION:
CEDAR BRANCH 25.0
END DESCRIPTION:
XS GIS Cut Line= 3
      3747399.64     10524960.19      3746599.61     10524860.19
       3745999.6      10525460.2
#Sta/Elev= 30
  4211.2  261.42    4477   252.2  4624.4  246.62  4634.5  247.04  4644.6  245.83
  4745.4  241.33  4805.2  238.37  4926.8  237.33  4946.9  238.43  4967.1  235.62
  4974.6   230.2  4984.2  229.46    4987  228.96  4990.2  229.46  5007.4  230.36
  5014.9  237.43    5021  237.43  5034.6  239.83  5088.2  240.79  5102.3  240.23
  5116.5  236.81  5130.6  240.81  5144.7  242.64    5173  242.71  5284.5  246.51
  5287.9  246.66  5399.3  249.26  5455.9  252.07  5526.1  253.67    5866  259.15
#Mann= 9 ,-1 , 0
  4211.2     .16       0    4477     .05       0  4805.2     .16       0
  4984.2     .07       0  4990.2     .16       0  5034.6     .12       0
  5284.5     .16       0  5287.9     .08       0  5526.1     .05       0
Bank Sta=4745.4,5144.7
XS Rating Curve= 0 ,0
Exp/Cntr=0.3,0.1

Type RM Length L Ch R = 1 ,28228   ,654,654,654
BEGIN DESCRIPTION:
CEDAR BRANCH 24.0
END DESCRIPTION:
XS GIS Cut Line= 3
      3747299.59     10524610.18      3746599.61     10524410.19
      3745899.61     10524510.19
#Sta/Elev= 30
  4308.5  259.13    4432  255.64  4476.2  252.29  4526.9  250.49  4616.6  245.34
  4641.3  245.07  4689.4  242.44  4694.6  243.96  4703.7  241.88  4734.9  240.26
  4828.5  238.68    4835  237.74  4880.5  237.82  4890.9  236.81  4932.5  237.13
  4953.3  235.19  4974.1  235.55  4980.6  235.42  4985.8  232.25  4994.9  228.46
    4997  228.46  4999.8  227.96    5003  228.46  5005.3  231.02  5026.1  236.33
    5087   241.6  5137.5  243.35  5309.2  249.54    5390  250.06  5743.6  258.18
#Mann= 4 ,-1 , 0
  4308.5     .16       0    4997     .07       0    5003     .16       0
  5137.5     .05       0
Bank Sta=4974.1,5087
XS Rating Curve= 0 ,0
Exp/Cntr=0.3,0.1

Type RM Length L Ch R = 1 ,27574   ,915,915,915
BEGIN DESCRIPTION:
CEDAR BRANCH 23.0
END DESCRIPTION:
XS GIS Cut Line= 3
      3747480.49     10523877.28      3746334.69     10523946.73
      3745702.83     10523964.04
#Sta/Elev= 30
  4271.7  259.33  4372.8  257.77  4452.9  258.82  4567.9  256.17  4691.2  250.48
  4875.8  240.48  4883.7  240.28  4973.9  234.98  4983.9  233.12  4990.9  228.13
  4993.7  227.63  4996.9  228.13  5003.9  230.36    5034  234.39  5061.3  236.45
  5124.1  234.12  5144.2     237  5204.3  235.03  5234.3  237.68  5262.4   238.3
  5294.5  241.27  5304.5  243.99  5314.5  244.43  5419.6  245.73  5424.7  243.41
  5464.7  243.14  5574.7   249.1  5604.8  248.85  5774.8  254.33  6051.7  257.71
#Mann= 6 ,-1 , 0
  4271.7     .16       0  4691.2     .05       0  4875.8     .16       0
  4990.9     .07       0  4996.9     .16       0  5262.4     .05       0
Bank Sta=4883.7,5294.5
XS Rating Curve= 0 ,0
Exp/Cntr=0.3,0.1

Type RM Length L Ch R = 1 ,26659   ,555,555,555
BEGIN DESCRIPTION:
CEDAR BRANCH 21.0
END DESCRIPTION:
XS GIS Cut Line= 3
      3747277.85     10523728.63      3746626.79     10523431.75
      3746056.44     10523421.33
#Sta/Elev= 30
  4429.7  255.43  4557.1  253.59  4570.2   253.4  4602.4   253.1  4682.5  249.71
  4700.1  250.04  4790.5  245.16  4797.7  244.04  4878.4  238.91  4941.5  234.06
  4964.5  234.48  4987.6  231.43  4989.6  230.36  4999.3  225.69  5007.3  225.25
    5010  224.75  5013.3  225.25  5016.1  228.74  5021.6  232.73  5054.2  232.19
  5088.3  235.57  5162.4  239.24  5262.5   243.5    5344   243.6  5432.5  246.48
  5592.5  249.56  5602.5  250.74  5622.5  250.73  5642.5  252.02  5715.7  253.18
#Mann= 8 ,-1 , 0
  4429.7     .16       0  4557.1     .05       0  4570.2     .16       0
  4989.6     .12       0  5007.3     .07       0  5013.3     .12       0
  5088.3     .16       0    5344     .05       0
Bank Sta=4878.4,5162.4
XS Rating Curve= 0 ,0
Exp/Cntr=0.3,0.1

Type RM Length L Ch R = 1 ,26104   ,509,509,509
BEGIN DESCRIPTION:
CEDAR BRANCH 20.0
END DESCRIPTION:
XS GIS Cut Line= 3
      3747421.03     10523080.19      3746600.75     10523116.65
      3746114.19     10523088.03
#Sta/Elev= 30
  4305.5   255.3  4326.9  253.56  4390.5  252.91  4447.1  251.92  4527.1  247.99
  4607.2  242.13  4727.3  237.34  4857.5  233.19  4927.5  234.09  4957.6  231.09
  4987.6  231.23  4997.6  224.13  5004.6  224.11  5007.4  223.61  5010.6  224.11
  5017.6  233.85  5037.6  237.45  5117.7  242.09  5152.1  241.76  5187.8  236.99
  5217.9  236.35  5237.9  237.46  5247.9  236.32    5258  237.36  5322.4  243.84
  5328.1  242.01  5340.5  241.95  5438.3  246.41  5572.2  250.46    5614  251.58
#Mann= 6 ,-1 , 0
  4305.5     .05       0  4390.5     .16       0  5004.6     .07       0
  5010.6     .16       0  5340.5     .05       0  5572.2     .16       0
Bank Sta=4727.3,5258
XS Rating Curve= 0 ,0
Exp/Cntr=0.3,0.1

Type RM Length L Ch R = 1 ,25595   ,620,620,620
BEGIN DESCRIPTION:
CEDAR BRANCH 19.0
END DESCRIPTION:
XS GIS Cut Line= 3
      3747249.61     10522960.19      3746849.61     10522710.19
      3746249.57     10522510.17
#Sta/Elev= 30
  4550.8  249.75    4674  244.36  4725.9  243.27  4774.9  239.61  4820.9  237.51
  4841.5  236.02  4892.8  231.96  4978.3  233.38  4987.1  223.13  4996.5  222.33
  4999.3  221.83  5002.5  222.33  5008.9  226.15  5014.8  225.31  5019.6  229.09
  5025.1  229.09    5033  230.98  5085.7  230.54  5138.5  233.62  5191.2  235.31
  5201.7  236.63  5264.9   239.6    5286   239.6  5296.6  241.04  5349.3  243.66
    5402  244.26  5445.4  246.44  5570.6  250.16  5581.2  251.36    5655  253.96
#Mann= 5 ,-1 , 0
  4550.8     .05       0  4820.9     .16       0  4996.5     .07       0
  5002.5     .16       0  5445.4     .05       0
Bank Sta=4841.5,5201.7
XS Rating Curve= 0 ,0
Exp/Cntr=0.3,0.1

Type RM Length L Ch R = 1 ,24975   ,488,488,488
BEGIN DESCRIPTION:
CEDAR BRANCH 18.0
END DESCRIPTION:
XS GIS Cut Line= 4
      3747844.02     10522810.41      3747198.18     10522324.28
      3746753.73     10522442.34      3746038.42     10522352.06
#Sta/Elev= 30
  3913.5   254.4  4081.7  251.87  4102.8  252.84  4217.3  250.26  4523.4  239.68
  4765.6   234.8  4805.8  234.21    4921   229.1    4979  228.65  4996.3  220.38
  4998.5  220.15  5001.2  219.65  5004.5  220.15  5010.1  227.86  5020.4  229.62
  5071.5  229.88  5111.6  233.72    5157  235.16  5181.3  237.34  5226.2   238.9
    5235  240.32  5240.1  239.18    5327  243.56  5410.3  246.13  5488.2   247.9
  5568.9  251.68  5669.7  254.82  5716.5   254.7  5760.4  256.18  5902.7  256.43
#Mann= 5 ,-1 , 0
  3913.5     .05       0    4921     .16       0  4998.5     .07       0
  5004.5     .16       0  5410.3     .05       0
Bank Sta=4765.6,5157
XS Rating Curve= 0 ,0
Exp/Cntr=0.3,0.1

Type RM Length L Ch R = 1 ,24487   ,489,489,489
BEGIN DESCRIPTION:
CEDAR BRANCH 17.0
END DESCRIPTION:
XS GIS Cut Line= 3
      3747249.59     10521960.19      3746699.61     10522110.19
      3746499.63     10522160.18
#Sta/Elev= 30
    4424  240.97  4465.4  240.81  4515.5  238.59  4520.7  238.96  4555.3  235.73
  4620.9  234.21  4669.3   231.7  4693.5  231.26  4828.2     231  4880.1  229.63
  4897.3   230.4  4931.9  227.74  4983.7  227.94  4991.5  221.31  4996.6  221.31
  5001.4  220.21  5004.1  219.71  5007.4  220.21  5012.1  222.86  5017.3  228.31
    5025  234.01  5035.3  236.44  5045.6   240.1  5053.3  241.25  5058.5  240.93
  5066.2   242.6  5086.8  243.88  5099.7  243.67  5163.3   245.9  5200.2  246.74
#Mann= 4 ,-1 , 0
    4424     .16       0  5001.4     .07       0  5007.4     .16       0
  5163.3     .05       0
Bank Sta=4620.9,5025
XS Rating Curve= 0 ,0
Exp/Cntr=0.3,0.1

Type RM Length L Ch R = 1 ,23998   ,535,535,535
BEGIN DESCRIPTION:
CEDAR BRANCH 16.0
END DESCRIPTION:
XS GIS Cut Line= 3
      3747499.59     10521610.19      3746899.61     10521760.19
      3746399.58      10522010.2
#Sta/Elev= 30
    4382  251.22  4835.5  232.73    4918  227.67  4982.4  228.46  4990.1  219.36
  4994.9  217.78  4997.6  217.28  5000.9  217.78  5003.2  217.78  5008.8  226.96
  5067.5  228.12  5103.9  230.99  5120.6  234.32  5126.2  233.37    5143  235.71
  5148.6   234.3  5165.4  237.65  5170.9  236.38  5179.3  238.08  5282.7  238.54
  5299.5  240.16  5313.5  231.99  5321.9   233.5  5327.5  238.16  5349.8  233.61
  5358.2  234.33  5372.2  241.55  5477.5  245.92  5523.1  247.72  5559.5  246.47
#Mann= 4 ,-1 , 0
    4382     .16       0  4994.9     .07       0  5000.9     .16       0
  5477.5     .05       0
Bank Sta=4835.5,5321.9
XS Rating Curve= 0 ,0
Exp/Cntr=0.3,0.1

Type RM Length L Ch R = 1 ,23463   ,392,392,392
BEGIN DESCRIPTION:
CEDAR BRANCH 15.0
END DESCRIPTION:
XS GIS Cut Line= 3
      3747281.49     10520845.13       3746670.4     10521449.28
       3746288.7     10521775.46
#Sta/Elev= 30
  4299.1  256.97  4452.5  253.26  4537.4   248.5  4615.1  242.32  4834.4  231.74
  4883.8  230.63  4968.7  227.18  4975.8  220.78  4986.9  216.88  4989.7  216.38
  4992.9  216.88    4997  217.43  5004.1  223.64  5018.2  225.96  5049.9  226.88
  5081.8  227.07  5103.1   229.1  5124.3  229.46  5138.4  231.36  5198.7  231.49
  5223.9  231.59  5244.7  233.45  5287.5  233.01  5336.9  235.06  5357.8  234.69
  5414.9  238.66  5443.4  237.33  5500.5  241.39  5558.1  242.08  5660.5  244.73
#Mann= 6 ,-1 , 0
  4299.1     .16       0  4986.9     .07       0  4992.9     .16       0
  5049.9     .12       0  5198.7     .16       0  5558.1     .05       0
Bank Sta=4883.8,5138.4
XS Rating Curve= 0 ,0
Exp/Cntr=0.3,0.1

Type RM Length L Ch R = 1 ,23071   ,493,493,493
BEGIN DESCRIPTION:
CEDAR BRANCH 14.0
END DESCRIPTION:
XS GIS Cut Line= 3
      3746699.61     10520810.18      3746499.61     10521210.19
      3746199.61     10521560.19
#Sta/Elev= 30
  4545.3  247.83  4616.1  241.98  4723.3  235.07  4791.3  230.03  4833.9  225.87
  4894.7  227.33  4939.4  225.66  4956.2  216.93  4961.8  225.49  4970.2  222.62
  4984.1  222.82  4989.7  219.02  4995.8  219.02  4996.7  216.79  4999.4  216.29
  5002.7  216.79  5013.9  218.37  5028.2  229.11  5042.5  226.28    5049  220.55
  5063.3  225.98    5071  225.38  5077.6  229.55    5127  230.08  5134.7  228.75
  5141.2  229.98  5162.3  230.34  5253.1  231.89  5361.3  235.08  5453.5  240.73
#Mann= 8 ,-1 , 0
  4545.3     .16       0  4616.1     .12       0  4723.3     .16       0
  4833.9     .12       0  4996.7     .07       0  5002.7     .12       0
  5162.3     .16       0  5253.1     .05       0
Bank Sta=4791.3,5141.2
XS Rating Curve= 0 ,0
Exp/Cntr=0.3,0.1

Type RM Length L Ch R = 1 ,22578   ,401,401,401
BEGIN DESCRIPTION:
CEDAR BRANCH 13.0
END DESCRIPTION:
XS GIS Cut Line= 3
      3746449.62     10520710.18      3746299.61     10520860.19
      3745999.62     10521210.17
#Sta/Elev= 30
    4770  242.11  4784.2  240.26    4804  239.49  4840.7   235.6  4875.9  233.47
  4883.1  233.18  4897.3  231.16  4911.4  225.06  4939.7  221.44  4946.8  222.76
    4968  224.63  4989.3  223.51  4995.9  219.91  5000.5  215.55  5003.3  215.05
  5006.5  215.55  5010.1  221.03  5017.8  226.91  5052.9  228.16  5096.5  227.73
  5194.5  227.14  5208.8  227.77  5280.1  227.52  5286.7  228.18  5337.2  229.49
  5343.8  230.52  5378.9  231.49  5429.4  233.96    5436  235.26  5443.1  235.24
#Mann= 6 ,-1 , 0
    4770     .16       0    4804     .12       0  4875.9     .16       0
  5000.5     .07       0  5006.5     .16       0  5096.5     .05       0
Bank Sta=4897.3,5286.7
XS Rating Curve= 0 ,0
Exp/Cntr=0.3,0.1

Type RM Length L Ch R = 1 ,22177   ,716,716,716
BEGIN DESCRIPTION:
CEDAR BRANCH 12.0
END DESCRIPTION:
XS GIS Cut Line= 3
      3746499.59     10520260.21      3746003.73     10520817.34
      3745849.61     10521710.19
#Sta/Elev= 30
  4328.4  254.25  4337.5  254.15  4470.1  248.42  4555.4  242.46  4710.9  236.51
    4746  233.34  4888.2   227.8  4930.8  225.49  4937.5  223.52  4980.2  223.52
  4986.9  221.44  4998.1  214.97  5000.8  214.47  5004.1  214.97  5008.6  219.98
  5022.8  221.54  5029.5  219.18  5037.2  220.09  5043.7  220.05  5057.9  224.86
  5072.1   226.2  5117.7  223.02    5138  226.86  5148.2  228.24  5190.2  231.66
  5351.1  231.58  5424.5  235.79  5544.2  239.67  5767.2  243.07  5980.3  249.72
#Mann= 6 ,-1 , 0
  4328.4     .16       0  4337.5     .05       0  4998.1     .03       0
  5004.1     .05       0  5037.2     .12       0    5138     .05       0
Bank Sta=4888.2,5148.2
XS Rating Curve= 0 ,0
Exp/Cntr=0.3,0.1
