HEC-RAS study HURRICANE BAYOU.prj: HURRICANE BAYOU Base Level Engineering

--- HURRICANE BAYOU.g01 (geometry) --- (continued)

Type RM Length L Ch R = 1 ,151655  ,312,312,312
BEGIN DESCRIPTION:
Mapping XS 1616ccc8
END DESCRIPTION:
XS GIS Cut Line= 3
      3833589.85     10491890.08       3832650.4     10492619.67
      3832567.93     10494030.28
#Sta/Elev= 30
  3760.1  353.87  3831.8  351.16    3925  344.78  3937.7  344.89  3966.7  341.43
    4039  336.77  4066.2   333.4  4124.2  330.64  4507.9  322.19    4545  322.74
    4736  319.28  4970.1  318.92  4980.2  316.85  4990.2  307.77  4997.2  307.47
  4999.9  306.97  5003.2  307.47  5010.2  307.97  5020.2   312.4  5030.2  319.14
  5260.6  318.95    5471   320.5  5551.1  324.45  5621.2  330.04  5631.3  331.88
  5661.3  332.62  5751.5  340.72  5901.1  345.07    6082  343.78  6362.6  344.55
#Mann= 3 ,-1 , 0
  3760.1     .05       0  4997.2     .03       0  5003.2     .05       0
Bank Sta=4970.1,5030.2
XS Rating Curve= 0 ,0
Exp/Cntr=0.3,0.1

Type RM Length L Ch R = 1 ,151343  ,1002,1002,1002
BEGIN DESCRIPTION:
HURRICANE BAYOU 126.0
END DESCRIPTION:
XS GIS Cut Line= 3
      3832289.44     10491483.47      3832487.36     10493228.23
      3832570.58     10493946.07
#Sta/Elev= 30
  3649.5  359.87  4008.5  342.99  4109.1  334.83  4129.3  332.14  4300.4  322.34
  4531.8  317.08  4642.5  316.48  4793.5  318.08    4864  317.07  4954.5  318.65
  4974.7  313.81  4981.7  307.69  4984.5  307.19  4987.7  307.69  4994.8  307.81
  5004.9  313.83  5014.9  317.61  5023.1  318.92  5065.2  317.33  5125.6  317.49
  5357.1  321.74  5470.6  329.81  5477.9  331.56  5508.1  332.33  5538.3  335.79
  5568.5  336.73  5598.7  339.97  5731.8  344.19  5899.1  343.35  6128.1  344.25
#Mann= 3 ,-1 , 0
  3649.5     .05       0  4981.7     .03       0  4987.7     .05       0
Bank Sta=4954.5,5023.1
XS Rating Curve= 0 ,0
Exp/Cntr=0.3,0.1

Type RM Length L Ch R = 1 ,150341  ,744,744,744
BEGIN DESCRIPTION:
HURRICANE BAYOU 125.0
END DESCRIPTION:
XS GIS Cut Line= 3
      3832185.27     10491504.25      3832023.81     10493525.11
      3832444.54      10494065.3
#Sta/Elev= 30
  3279.6  360.59  3405.9  353.27  3535.2  341.12  3668.2  332.89  3967.7   318.1
  4308.8  314.72    4369  316.66  4429.2  315.61    4539  317.91  4700.1  315.18
  4910.7  316.79  4970.9   314.2  4988.5  308.41    4998  306.64  5000.8  306.14
    5004  306.64    5011  312.53  5031.1  321.89    5041  322.35  5061.2  319.93
  5071.2  323.22  5085.2  323.73  5168.9  329.27  5181.6   328.7  5240.7  333.85
  5392.6  337.87  5649.6  337.42    5807   340.3  5842.3  342.57  5991.6  343.39
#Mann= 6 ,-1 , 0
  3279.6     .05       0  4988.5     .16       0    4998     .07       0
    5004     .16       0  5085.2      .1       0  5240.7     .05       0
Bank Sta=4910.7,5031.1
XS Rating Curve= 0 ,0
Exp/Cntr=0.3,0.1

Type RM Length L Ch R = 1 ,149597  ,373,373,373
BEGIN DESCRIPTION:
HURRICANE BAYOU 124.0
END DESCRIPTION:
XS GIS Cut Line= 3
       3832049.6     10491510.23      3831749.61     10492710.19
      3831549.62     10493610.15
#Sta/Elev= 30
  3727.1  359.27  3832.7  352.21  3992.5  336.72  4038.9  335.23  4116.2  328.41
  4203.8  325.04  4252.8  320.71  4551.7  315.83  4891.8  313.97  4953.7  315.09
  4966.6  313.53  4978.1  305.42  4980.2  303.95  4982.9  303.45  4986.2  303.95
  4988.3   308.2  4994.7  306.58  5015.2  306.63  5025.5  312.67  5031.9  314.11
    5037  312.54  5057.6  313.82  5157.3  315.38  5250.8  314.51    5302  316.52
  5414.7  316.53  5660.6  320.51  5752.8  325.34    5804  331.69  5885.9  335.62
#Mann= 6 ,-1 , 0
  3727.1     .05       0  4978.1     .16       0  4980.2     .07       0
  4986.2     .16       0  5057.6     .12       0  5157.3     .05       0
Bank Sta=4953.7,5031.9
XS Rating Curve= 0 ,0
Exp/Cntr=0.3,0.1

Type RM Length L Ch R = 1 ,149224  ,842,842,842
BEGIN DESCRIPTION:
HURRICANE BAYOU 123.0
END DESCRIPTION:
XS GIS Cut Line= 3
       3831949.6     10491360.22      3831449.61     10492560.19
      3831449.61     10493660.22
#Sta/Elev= 30
  3654.9  368.15  3823.3  353.75  4006.4  341.53  4380.7  321.25  4449.5  321.98
  4662.4  314.65  4762.6  314.61  4792.4  311.13  4803.2  313.95    4861  314.66
  4887.2  315.57  4892.9  315.42  4940.2  311.71  4945.7  308.31  4957.4   308.2
  4964.9  311.45  4975.7  310.32  4984.9  311.21  4994.9  304.67  5001.9  304.17
  5004.6  303.67  5007.9  304.17  5024.9  305.01  5034.9  312.07  5044.9  314.41
  5185.6  313.35  5283.7  314.32  5574.9  316.55  5844.9  329.95  6054.9  337.08
#Mann= 8 ,-1 , 0
  3654.9     .05       0    4861     .12       0  4892.9     .16       0
  4975.7     .12       0  5001.9     .07       0  5007.9     .12       0
  5185.6     .16       0  5283.7     .05       0
Bank Sta=4887.2,5044.9
XS Rating Curve= 0 ,0
Exp/Cntr=0.3,0.1

Type RM Length L Ch R = 1 ,148382  ,1353,1353,1353
BEGIN DESCRIPTION:
HURRICANE BAYOU 122.0
END DESCRIPTION:
XS GIS Cut Line= 3
      3830959.01     10491283.72      3830986.79     10492686.52
       3831299.3     10493721.28
#Sta/Elev= 30
  4065.5  370.12  4082.2  368.42    4282  355.77    4462   339.1  4532.1  334.72
  4602.1  338.96  4671.5  340.32  4769.7  339.41  4832.1  336.97  4872.1  330.01
  4931.9  323.01  4962.1  314.36  4992.2  309.64  4999.2  304.09  5001.9  303.59
  5005.2  304.09  5012.2  304.19  5032.2  311.01  5052.2  312.44  5092.2  311.03
  5118.5  313.65  5232.2   313.8  5302.2  311.19  5457.2  312.18  5462.9   312.1
  5560.3  314.16  5994.7  313.65  6149.5  318.13  6402.1  333.43  6549.5  336.14
#Mann= 11 ,-1 , 0
  4065.5     .05       0  4082.2     .16       0  4671.5      .1       0
  4769.7     .16       0  4931.9     .12       0  4999.2     .07       0
  5005.2     .12       0  5118.5     .16       0  5457.2     .05       0
  5462.9     .16       0  5560.3     .05       0
#XS Ineff= 1 ,-1
    4462  4652.1     340
Permanent Ineff=
       F
Bank Sta=4962.1,5052.2
XS Rating Curve= 0 ,0
Exp/Cntr=0.3,0.1

Type RM Length L Ch R = 1 ,147029  ,1621,1621,1621
BEGIN DESCRIPTION:
HURRICANE BAYOU 121.0
END DESCRIPTION:
XS GIS Cut Line= 3
       3830434.4      10491655.4      3830399.68     10493204.02
      3831413.55     10494162.33
#Sta/Elev= 30
  3839.6  350.04  3944.4   345.4  4074.5  342.47  4154.5  338.09  4214.5  333.94
  4294.5  322.26  4352.8  316.62  4454.5  312.58  4687.9  310.51  4726.2  311.29
  4744.6  309.92  4774.6  304.23  4811.4  308.56  4844.6  309.56  4854.6  305.53
  4954.7  309.49  4974.7  307.64  4984.7  301.91  4994.3  301.38  5001.7  300.34
  5004.4  299.84  5007.7  300.34  5014.7  302.95  5024.7  311.15  5164.3  310.74
  5194.7  308.46  5384.2  310.93  6192.2  313.96  6553.1  337.39  6783.7  339.63
#Mann= 7 ,-1 , 0
  3839.6     .05       0  4352.8     .16       0  4687.9     .12       0
  4811.4     .16       0  4994.3     .05       0  5001.7     .03       0
  5007.7     .05       0
Bank Sta=4954.7,5024.7
XS Rating Curve= 0 ,0
Exp/Cntr=0.3,0.1

Type RM Length L Ch R = 1 ,145408  ,381,381,381
BEGIN DESCRIPTION:
HURRICANE BAYOU 120.0
END DESCRIPTION:
XS GIS Cut Line= 3
      3830249.63     10491910.16      3829649.61     10492710.19
       3829399.6     10494260.22
#Sta/Elev= 30
  4000.2  326.25  4263.8  312.81  4378.4  309.51  4863.8  308.78  4950.2  309.73
  4957.5  304.28  4978.4  302.31  4986.7  298.95  4992.9  300.57  4994.1   296.3
  4996.9   295.8  5000.1   296.3  5006.9  296.48  5010.4  296.64  5020.5  301.06
  5028.6  301.99  5033.7  300.91  5040.8  303.19  5071.1  304.52  5090.3  308.02
  5095.5  308.25  5131.9  306.71  5152.2  307.69  5182.6  305.93  5476.3     315
    5608  316.75  5718.4  314.96    5922  316.73  6387.9  325.74  6570.3  332.28
#Mann= 5 ,-1 , 0
  4000.2     .05       0  4994.1     .03       0  5000.1     .05       0
  5006.9     .16       0  5090.3     .05       0
Bank Sta=4950.2,5095.5
XS Rating Curve= 0 ,0
Exp/Cntr=0.3,0.1

Type RM Length L Ch R = 1 ,145027  ,755,755,755
BEGIN DESCRIPTION:
HURRICANE BAYOU 119.0
END DESCRIPTION:
XS GIS Cut Line= 3
      3830264.29     10491285.58      3829153.15     10492952.28
      3828849.32     10493690.15
#Sta/Elev= 30
  3243.7  359.14  3309.3  356.49  3459.5  345.42  3618.7  338.39  3675.8  338.19
  3747.9  335.36  3862.2  319.94  4006.4  310.18  4390.9  307.34  4628.3  308.66
  4799.6   307.3  4835.7  308.46  4859.7   307.4  4871.7  305.17  4931.8  304.97
  4952.8  306.18  4967.8  303.83  4973.8  306.53  4979.9  299.11  4988.9  296.87
  5000.9  296.61  5003.6  296.11  5006.9  296.61    5016  300.93  5024.9  302.99
    5061  308.13    5076  311.13  5154.1  317.76  5536.9  319.49  6044.8   324.8
#Mann= 3 ,-1 , 0
  3243.7     .05       0  5000.9     .03       0  5006.9     .05       0
Bank Sta=4973.8,5061
XS Rating Curve= 0 ,0
Exp/Cntr=0.3,0.1

Type RM Length L Ch R = 1 ,144272  ,880,880,880
BEGIN DESCRIPTION:
HURRICANE BAYOU 118.0
END DESCRIPTION:
XS GIS Cut Line= 2
      3829526.42     10491007.82      3828667.24     10493385.76
#Sta/Elev= 30
  3430.2  353.96    3656  340.41  3751.7  331.78  3758.1  329.91  3826.1   322.8
  3889.9  317.69  3900.6   315.4  3962.1   312.1  4084.8  312.51  4091.9  309.45
  4115.5  308.64  4485.4  305.37    4900   307.1  4911.5  303.87  4953.2  304.11
  4967.5  302.66  4995.1  295.91  4997.9  295.41  5001.1  295.91    5017  296.83
  5023.5  302.74  5028.8  302.95  5038.3  307.03  5079.5  309.94  5319.5     313
  5462.2  316.68  5579.5  317.57  5615.5  316.72  5671.5  318.72  5958.6  321.38
#Mann= 3 ,-1 , 0
  3430.2     .05       0  4995.1     .03       0  5001.1     .05       0
Bank Sta=4900,5038.3
XS Rating Curve= 0 ,0
Exp/Cntr=0.3,0.1

Type RM Length L Ch R = 1 ,143392  ,545,545,545
BEGIN DESCRIPTION:
HURRICANE BAYOU 117.0
END DESCRIPTION:
XS GIS Cut Line= 3
      3829326.78      10490877.6      3828502.11     10492066.86
      3828519.47     10493464.44
#Sta/Elev= 30
  2920.4  349.78  3013.4  345.84  3081.6  340.45  3099.9  340.16  3179.1  330.49
  3257.9  325.96  3272.8   323.6  3293.7  324.18    3459  312.59    3568  307.93
  4048.3  305.07  4113.8  303.21  4128.3  304.57    4611  306.45    4631  302.23
    4641  301.77    4761  303.54    4821  306.35    4951  301.66  4997.1  294.78
    4998  294.69  5000.7  294.19    5004  294.69    5021  296.29    5041  303.71
    5061  306.91    5106  307.71    5331  312.04    5421  315.85  5765.3  322.28
#Mann= 6 ,-1 , 0
  2920.4      .1       0  3081.6     .05       0  4997.1     .16       0
    4998     .07       0    5004     .16       0    5106     .05       0
Bank Sta=4821,5061
XS Rating Curve= 0 ,0
Exp/Cntr=0.3,0.1

Type RM Length L Ch R = 1 ,142847  ,2985,2985,2985
BEGIN DESCRIPTION:
HURRICANE BAYOU 116.0
END DESCRIPTION:
XS GIS Cut Line= 4
      3829475.79     10490569.46      3828347.31      10491715.3
      3828165.02     10492756.97      3828555.11     10493649.84
#Sta/Elev= 30
  2746.8  350.49  2846.6  346.72  2900.2  341.52  2949.7  340.31  3105.3  346.82
  3216.2  344.53  3402.3  337.21  3567.4  320.38  3642.7  313.67  3754.7  308.14
  4432.4  304.21  4461.5  300.38  4512.3  303.52    4695  305.02  4969.1  304.17
  4979.3  294.21  4986.4  293.26  4989.2  292.76  4992.4  293.26    5030  300.54
  5101.1   305.3    5162  305.46  5185.1  299.39  5202.6  304.25  5263.5  302.74
  5290.5  304.94  5434.5  308.73  5713.7  309.54  5994.4  319.01  6386.9  326.67
#Mann= 8 ,-1 , 0
  2746.8     .05       0  2846.6      .1       0  3216.2     .05       0
  3567.4      .1       0  3754.7     .16       0  4986.4     .07       0
  4992.4     .16       0  5290.5     .05       0
#XS Ineff= 1 ,-1
  2850.7  3098.2  346.13
Permanent Ineff=
       F
Bank Sta=4969.1,5101.1
XS Rating Curve= 0 ,0
Exp/Cntr=0.3,0.1

Type RM Length L Ch R = 1 ,139862  ,156,156,156
BEGIN DESCRIPTION:
HURRICANE BAYOU 113.0
END DESCRIPTION:
XS GIS Cut Line= 6
      3826414.43     10490217.88       3826700.9      10491381.1
      3826831.11     10491845.51      3827069.82     10492197.07
      3827738.22     10492787.35      3828423.99     10493620.69
#Sta/Elev= 30
  3668.3  335.92  3892.1   323.9  4001.4  319.11  4098.6  314.95  4205.5  309.62
  4307.5  306.33  4456.7  302.15  4715.5  300.34  4817.6  300.93  4886.1  300.71
    4938  298.82  4997.3  287.47  5000.1  286.97  5003.3  287.47  5023.1  294.72
  5052.3  298.89  5142.3  298.77  5408.6  300.44  5575.2  298.67  5876.9  302.67
  6004.5   303.6    6427  314.12  6642.4  313.26  6743.2  312.18  6945.1  309.51
  6988.2  314.63  7037.7  310.19  7115.9   316.8  7579.2  323.19  7744.5   325.7
#Mann= 20 ,-1 , 0
  3668.3     .16       0  3892.1     .05       0  4001.4     .08       0
  4098.6     .05       0  4205.5     .08       0  4307.5     .05       0
  4456.7     .08       0  4715.5     .05       0  4817.6     .12       0
  4997.3     .07       0  5003.3     .08       0  5023.1     .05       0
  5142.3     .16       0  5408.6     .16       0  5575.2     .16       0
  5876.9     .16       0  6004.5     .16       0  6642.4     .16       0
  6743.2     .05       0  7579.2     .05       0
#XS Ineff= 1 ,-1
  6895.6  7101.5  314.42
Permanent Ineff=
       F
Bank Sta=4886.1,5052.3
XS Rating Curve= 0 ,0
Exp/Cntr=0.3,0.1

Type RM Length L Ch R = 1 ,139706  ,778,778,778
BEGIN DESCRIPTION:
HURRICANE BAYOU 112.0
END DESCRIPTION:
XS GIS Cut Line= 6
      3826375.39     10490174.46      3826297.25      10490530.4
      3826670.52     10491819.47      3826861.49     10492335.96
      3827720.86     10493121.55       3827920.5     10493642.36
#Sta/Elev= 30
  3612.7  337.24  3756.5  327.19  3781.4  322.51  3828.3  322.05  3876.7  318.92
  3980.8  315.93  4060.9  312.87  4509.7  299.04  4842.1  299.65  4933.6  295.55
  4977.7  298.54  4986.8  289.12  5003.1  284.82  5005.8  284.32  5009.1  284.82
    5018  285.04  5044.9  295.78    5151  300.12  5295.4  300.23  5323.7  300.35
  5535.9  301.38  5576.2  300.75  5607.8  297.64  5646.6  301.51  5748.2   301.6
  6308.3  309.08  6422.9  311.32  7025.2  323.04  7325.6  319.74  7591.9  333.93
#Mann= 16 ,-1 , 0
  3612.7     .16       0  3781.4     .08       0  3828.3     .05       0
  3876.7     .16       0  3980.8     .12       0  4060.9     .05       0
  4842.1     .12       0  5003.1     .07       0  5009.1     .12       0
  5295.4     .05       0  5323.7     .08       0  5535.9     .05       0
  5576.2     .08       0  5748.2     .05       0  6308.3     .08       0
  6422.9     .05       0
Bank Sta=4977.7,5151
XS Rating Curve= 0 ,0
Exp/Cntr=0.3,0.1

Type RM Length L Ch R = 1 ,138928  ,773,773,773
BEGIN DESCRIPTION:
HURRICANE BAYOU 111.0
END DESCRIPTION:
XS GIS Cut Line= 3
      3826308.38     10490100.31       3825733.3     10491912.35
      3825396.93     10493843.77
#Sta/Elev= 30
  3528.7  332.36    3602  333.12  3646.1  329.86  3677.1  323.14  3741.6  320.13
  3773.9  323.93  3820.6  322.62  3902.9  319.85  4080.3  307.69    4182  303.96
  4328.1  299.23  4394.6  297.76  4639.3  298.61  4792.3  295.99  4859.6  297.42
  4897.1  296.25  4913.5  292.51  4929.4  295.33  4961.7  294.61  4986.9  290.83
  4996.2  283.93  4998.9  283.43  5002.2  283.93  5026.2  285.19  5031.5  292.14
  5049.8  296.13    5096  297.98  5823.5  306.73  6371.6  325.83  7390.3  329.33
#Mann= 11 ,-1 , 0
  3528.7     .16       0  3646.1     .05       0  3820.6     .16       0
  4080.3     .12       0    4182     .05       0  4328.1     .16       0
  4394.6     .05       0  4639.3     .16       0  4792.3     .05       0
  4996.2     .03       0  5002.2     .05       0
Bank Sta=4859.6,5096
XS Rating Curve= 0 ,0
Exp/Cntr=0.3,0.1

Type RM Length L Ch R = 1 ,138155  ,1321,1321,1321
BEGIN DESCRIPTION:
HURRICANE BAYOU 109.0
END DESCRIPTION:
XS GIS Cut Line= 3
       3826254.1     10490078.61      3825559.69     10490653.67
      3825028.01     10493453.12
#Sta/Elev= 30
  3695.5  329.16  3735.5  328.83  3764.1  328.58    3785  321.71  3834.5  320.46
  3863.1  326.17  3892.8  325.62    3997  322.35  4109.3  319.64  4246.7  309.23
  4375.4  304.53  4645.9  300.03  4890.4  296.01  4939.6  296.69  4987.5  282.54
  4990.3  282.04  4993.5  282.54  5002.7  283.49  5010.9  293.26  5035.9  295.73
    5072  296.72  5257.3  295.01  5367.1  298.77  5644.9  297.09  6067.9   306.7
  6396.6  310.31  6843.1  325.71  7152.3  324.97  7305.1   327.9  7446.6  327.11
#Mann= 13 ,-1 , 0
  3695.5     .16       0  3735.5     .05       0  3892.8     .16       0
    3997     .12       0  4109.3     .16       0  4375.4     .12       0
  4645.9     .05       0  4890.4     .16       0  4987.5     .07       0
  4993.5     .16       0  5035.9     .12       0  5257.3     .05       0
  7152.3     .16       0
#XS Ineff= 1 ,-1
  3770.6  3863.1  326.17
Permanent Ineff=
       F
Bank Sta=4939.6,5072
XS Rating Curve= 0 ,0
Exp/Cntr=0.3,0.1

Type RM Length L Ch R = 1 ,136834  ,507,507,507
BEGIN DESCRIPTION:
HURRICANE BAYOU 108.0
END DESCRIPTION:
XS GIS Cut Line= 3
      3825649.59     10489260.23      3824699.61     10490860.19
      3824899.61     10492660.18
#Sta/Elev= 30
  3158.9   377.5  3262.1  375.79  3347.8  355.86  3384.4  352.49  3400.5  350.02
  3421.9  338.52  3464.7  342.45  3545.5  337.48  4021.3  315.89  4129.6  312.24
    4914  294.36  4936.4  294.39  4938.2  294.36  4953.4  293.13  4981.6  280.61
  4984.3  280.11  4987.6  280.61    5006   285.4  5011.8  283.11  5016.7  288.26
  5029.7  290.39  5100.1  294.25  5223.2  294.99  5322.3  294.69  5604.3  295.11
    6227  300.32  6498.7  305.77  6697.6  314.76  6720.8   316.1  6830.7  321.69
#Mann= 14 ,-1 , 0
  3158.9     .16       0  3384.4     .05       0  3545.5     .16       0
  4021.3     .12       0  4129.6     .16       0    4914     .12       0
  4936.4     .16       0  4981.6     .07       0  4987.6     .16       0
  5223.2     .12       0  5322.3     .16       0  5604.3     .05       0
  6697.6     .16       0  6720.8     .05       0
Bank Sta=4938.2,5100.1
XS Rating Curve= 0 ,0
Exp/Cntr=0.3,0.1

Type RM Length L Ch R = 1 ,136327  ,622,622,622
BEGIN DESCRIPTION:
HURRICANE BAYOU 107.0
END DESCRIPTION:
XS GIS Cut Line= 3
      3825049.58     10489910.21      3824249.61     10490660.19
      3823912.42     10492683.33
#Sta/Elev= 30
  3894.3  316.23    4170  305.62  4578.3  297.11  4601.8  297.49  4693.6  290.95
  4778.6  293.66  4823.9  292.36    4879  293.98  4906.1  294.61  4948.6  292.96
  4962.7  288.99  4969.6  282.85  4984.4  280.68  4987.2  280.18  4990.4  280.68
    5001  281.47  5018.7  290.64  5051.7  293.97  5112.5  292.36  5254.4  293.78
  5295.6  290.47  5322.9  293.16  5609.3   297.1    5997  296.96  6366.5  302.42
  6424.4   303.6  6541.4  307.46  6769.7  314.73    6988  320.68  7041.9  319.45
#Mann= 11 ,-1 , 0
  3894.3     .16       0  4578.3     .12       0  4823.9     .16       0
    4879     .12       0  4984.4     .07       0  4990.4     .12       0
  5295.6     .16       0  6366.5     .12       0  6424.4     .16       0
  6541.4     .12       0  6769.7     .16       0
Bank Sta=4906.1,5051.7
XS Rating Curve= 0 ,0
Exp/Cntr=0.3,0.1

Type RM Length L Ch R = 1 ,135705  ,523,523,523
BEGIN DESCRIPTION:
HURRICANE BAYOU 106.0
END DESCRIPTION:
XS GIS Cut Line= 3
      3824399.61     10489610.19      3823899.54     10490394.38
      3823534.95     10492790.23
#Sta/Elev= 30
  4085.7  312.64  4389.7  299.18  4453.8  296.98  4484.3  289.76  4512.3  289.78
  4616.9  291.14  4707.8  289.76  4813.4  289.76  4963.3  293.61  4984.4  287.84
  4990.4  279.75  4998.3  280.05  5002.6  279.46  5005.3  278.96  5008.6  279.46
  5031.8  289.53  5052.8  293.17  5157.2  293.14  5532.8  291.81  5565.2  293.45
  5644.8  296.99  5734.1   297.1  6184.9  295.84  6642.9  312.86  6741.6  313.97
  6840.3  315.98  7121.5  318.58  7251.3  320.89  7273.7  320.86  7439.2  320.59
#Mann= 20 ,-1 , 0
  4085.7     .05       0  4389.7     .16       0  4512.3     .05       0
  4616.9     .12       0  4707.8     .05       0  4813.4     .12       0
  4998.3     .16       0  5002.6     .07       0  5008.6     .16       0
  5157.2     .12       0  5532.8     .05       0  5565.2     .16       0
  5644.8     .05       0  5734.1     .16       0  6642.9     .12       0
  6741.6     .16       0  6840.3     .12       0  7121.5     .16       0
  7251.3     .12       0  7273.7     .16       0
Bank Sta=4963.3,5052.8
XS Rating Curve= 0 ,0
Exp/Cntr=0.3,0.1

Type RM Length L Ch R = 1 ,135182  ,1007,1007,1007
BEGIN DESCRIPTION:
HURRICANE BAYOU 105.0
END DESCRIPTION:
XS GIS Cut Line= 4
      3824359.58     10489179.13      3823734.61     10489916.95
      3823465.51     10490316.26      3823487.06     10492526.09
#Sta/Elev= 30
  3749.2     323  3877.9  321.04  4104.4  313.44  4495.3  293.85    4865   289.8
  4945.9  292.65    4952  292.54  4960.9  287.21    4967  292.67  4973.3   291.7
  4980.4  283.18  4981.9  281.38    4988  283.37  4999.9   278.6  5002.7   278.1
  5005.9   278.6  5010.9  279.51  5017.9  283.69  5038.9   285.3  5045.6  290.92
  5059.9  289.72  5081.8  292.27  5095.8  292.37  5541.6  292.19  5631.6  289.64
  5791.6   297.6  6360.1  295.17  7172.4   313.9  7312.9  317.86  7407.6  319.56
#Mann= 9 ,-1 , 0
  3749.2     .05       0  4980.4     .12       0  4999.9     .07       0
  5005.9     .12       0  5010.9     .16       0  5095.8     .05       0
  6360.1     .16       0  7172.4     .12       0  7312.9     .16       0
Bank Sta=4967,5081.8
XS Rating Curve= 0 ,0
Exp/Cntr=0.3,0.1

Type RM Length L Ch R = 1 ,134175  ,639,639,639
BEGIN DESCRIPTION:
HURRICANE BAYOU 104.0
END DESCRIPTION:
XS GIS Cut Line= 3
      3822944.68     10489074.94      3823040.16     10490628.76
      3823365.53     10492474.96
#Sta/Elev= 30
  3926.2  322.07  3929.7  321.61  4011.6  316.75  4141.9  300.02  4238.6  292.17
    4484  289.19  4573.1   288.6  4702.9  290.58  4722.9  287.79  4739.1  291.31
  4940.1  291.16  4943.4  291.14  4963.4  288.22  4973.4  283.27  5000.5  277.75
  5003.2  277.25  5006.5  277.75  5023.5  277.92  5043.6  286.14  5065.8  288.05
  5133.7  291.27  5404.2  290.08  5514.9  292.47  5646.9  291.29  6215.5  294.13
  6464.3   299.5  6621.7  299.03  6868.3  302.04  6964.8  303.56  7357.6  318.53
#Mann= 12 ,-1 , 0
  3926.2     .05       0  3929.7     .16       0  4238.6     .05       0
    4484     .12       0  4573.1     .16       0  4940.1     .12       0
  5000.5     .07       0  5006.5     .12       0  5065.8     .05       0
  6464.3     .16       0  6868.3     .12       0  6964.8     .16       0
Bank Sta=4943.4,5133.7
XS Rating Curve= 0 ,0
Exp/Cntr=0.3,0.1

Type RM Length L Ch R = 1 ,133536  ,509,509,509
BEGIN DESCRIPTION:
HURRICANE BAYOU 103.0
END DESCRIPTION:
XS GIS Cut Line= 3
      3822745.03     10488988.12      3822493.29     10490437.78
      3823104.59     10492525.26
#Sta/Elev= 30
  3822.3  325.07    3958  312.47    4139  292.26  4362.9  287.07  4392.8  284.05
  4413.7  288.07    4473  288.63    4940   289.7  4971.3   289.2  4998.8  276.61
  5001.5  276.11  5004.8  276.61  5022.1  283.28  5046.3  284.05  5049.8  285.92
  5054.9  282.36  5072.8  289.66  5204.1  289.33  6069.2  296.91  6567.3  299.57
  6903.3  301.42  7052.2   306.1  7291.2   314.8  7324.7   316.1  7329.9  312.22
  7348.9  314.17  7369.7  310.06  7380.2  314.62  7413.4  316.91  7468.8  319.13
#Mann= 15 ,-1 , 0
  3822.3     .05       0    3958     .16       0  4362.9     .12       0
    4473     .16       0    4940     .12       0  4998.8     .07       0
  5004.8     .12       0  5046.3      .1       0  5204.1     .05       0
  6069.2     .12       0  6567.3     .16       0  6903.3     .12       0
  7052.2     .16       0  7291.2     .12       0  7413.4     .16       0
Bank Sta=4971.3,5072.8
XS Rating Curve= 0 ,0
Exp/Cntr=0.3,0.1

Type RM Length L Ch R = 1 ,133027  ,1434,1434,1434
BEGIN DESCRIPTION:
HURRICANE BAYOU 102.0
END DESCRIPTION:
XS GIS Cut Line= 3
      3822588.77     10488962.09       3822085.3     10490559.31
      3822736.15     10492355.64
#Sta/Elev= 30
  4077.8  326.67  4116.1  322.84    4221  311.28    4238  306.39  4339.7  294.06
  4400.8   289.2    4499  287.16  4560.4  285.39  4652.2  289.47  4786.9  287.63
    4967  289.43  4986.3  278.41  4995.5  275.96  4998.2  275.46  5001.5  275.96
  5023.9  283.39  5029.9  287.86  5050.9  288.88  5105.2  288.42  5356.3  289.52
  5423.5  287.63  5638.1  289.86  6008.7  288.17  6338.1  291.79  6457.6  292.91
    6857  297.68  7280.4  307.39  7433.9  314.28  7588.4  314.67  7663.1  314.43
#Mann= 15 ,-1 , 0
  4077.8     .16       0  4116.1     .05       0    4238     .16       0
  4339.7     .05       0    4499     .16       0  4995.5     .07       0
  5001.5     .16       0  5105.2     .12       0  5356.3      .1       0
  5423.5     .05       0  6338.1     .16       0  6457.6     .12       0
    6857     .16       0  7280.4     .12       0  7588.4     .16       0
Bank Sta=4967,5050.9
XS Rating Curve= 0 ,0
Exp/Cntr=0.3,0.1

Type RM Length L Ch R = 1 ,131593  ,498,498,498
BEGIN DESCRIPTION:
HURRICANE BAYOU 100.0
END DESCRIPTION:
XS GIS Cut Line= 3
      3822499.61     10488860.19      3821699.61     10489660.19
      3819699.59     10492060.21
#Sta/Elev= 30
  3834.6  331.17  3872.7  328.48    3976  320.52  4004.3   314.9  4179.5  293.64
    4385  285.02  4951.8  287.66  4987.5   281.4    4994   273.5  4998.8  272.92
  5001.5  272.42  5004.8  272.92  5030.4  273.96  5036.9  279.38  5044.1  279.25
  5051.2  285.24  5072.1   287.5  5104.1  287.01  5109.5  286.93  5242.6  285.33
    5335  289.51  5725.5  292.65  6520.9  293.81  6697.9  298.17  6812.4  305.07
  6996.6  297.11  7166.5  297.54  7756.2   313.7  7926.7  313.56  8090.1  318.66
#Mann= 8 ,-1 , 0
  3834.6     .05       0  3872.7     .16       0  4179.5     .05       0
    4385     .16       0  4998.8     .07       0  5004.8     .16       0
  5104.1     .16       0  5109.5     .05       0
Bank Sta=4951.8,5072.1
XS Rating Curve= 0 ,0
Exp/Cntr=0.3,0.1

Type RM Length L Ch R = 1 ,131095  ,580,580,580
BEGIN DESCRIPTION:
HURRICANE BAYOU 99.0
END DESCRIPTION:
XS GIS Cut Line= 3
      3822049.63     10488560.15      3821249.61     10489710.19
       3819649.6      10491710.2
#Sta/Elev= 30
  3630.4  336.22    3667  336.86  3800.7  326.76  3867.4  320.14  3945.4  307.06
  3995.9  298.64  4111.8  287.75  4269.8  285.32  4312.6  282.35  4320.4  284.98
  4484.5  286.76  4958.4   286.3  4973.3  281.75    4982  273.89  4991.8  272.71
  4994.5  272.21  4997.8  272.71  5009.1   274.3  5028.3  283.25  5087.4  288.34
  5415.5  293.81  5550.8  290.88  6027.8  291.76  6554.5   307.4  6703.3     300
  6802.6  300.16  6824.2  302.78  7044.3  310.39  7336.5  309.76  7592.6  315.72
#Mann= 6 ,-1 , 0
  3630.4     .05       0  3800.7     .12       0  3945.4     .16       0
  4991.8     .07       0  4997.8     .16       0  5087.4     .05       0
#XS Ineff= 1 ,-1
  6568.1  6980.3  307.16
Permanent Ineff=
       F
Bank Sta=4958.4,5087.4
XS Rating Curve= 0 ,0
Exp/Cntr=0.3,0.1

Type RM Length L Ch R = 1 ,130515  ,935,935,935
BEGIN DESCRIPTION:
HURRICANE BAYOU 98.0
END DESCRIPTION:
XS GIS Cut Line= 3
      3822198.21     10487509.49      3821049.61     10489210.19
      3819355.64      10491675.7
#Sta/Elev= 30
  2940.9  332.24  3732.8  330.31  3897.7   317.1  3915.1  310.12  3978.6  301.77
  4086.5  319.27  4143.4   322.3  4215.4  315.49  4293.3  297.77  4457.4  284.22
  4467.8   283.6  4539.1  284.86    4569  279.64  4712.9  286.34  4812.1  280.75
  4927.4  285.77  4934.7  286.55  4949.7  285.54  4982.7  271.68  4985.4  271.18
  4988.7  271.68  5000.6  273.43  5015.5  284.32  5045.2  286.02  5051.3  286.76
  5424.8  284.55    5619  291.41  6315.6  293.56  7007.2  307.98  7984.5  315.31
#Mann= 8 ,-1 , 0
  2940.9     .05       0  3915.1     .16       0  4457.4     .05       0
  4467.8     .16       0  4927.4     .12       0  4982.7     .07       0
  4988.7     .12       0  5045.2     .05       0
#XS Ineff= 1 ,-1
  3855.7  4136.4  321.95
Permanent Ineff=
       F
Bank Sta=4934.7,5051.3
XS Rating Curve= 0 ,0
Exp/Cntr=0.3,0.1

Type RM Length L Ch R = 1 ,129580  ,382,382,382
BEGIN DESCRIPTION:
HURRICANE BAYOU 97.0
END DESCRIPTION:
XS GIS Cut Line= 3
      3821937.77     10487466.12      3820581.44      10488876.7
      3819496.36     10491263.88
#Sta/Elev= 30
  3585.2  332.77  3869.6  334.29  3996.9  330.83  4244.4  331.69  4283.6  329.03
  4410.9  318.71  4447.7  315.48    4591  298.47  4698.4  291.46  4875.6  285.19
  4958.9  284.85    4973   283.8  4984.2  270.71  4986.9  270.21  4990.2  270.71
  5008.2  271.16  5015.5  276.39  5022.4  276.67  5029.6  283.51  5104.3  283.73
  5137.2  283.87  5635.2  285.01  5848.3  283.81  5871.3  281.45  5894.4  284.07
  5985.3   283.5    6280  290.37  6912.7  293.21  7539.9  307.38  8164.3  309.47
#Mann= 10 ,-1 , 0
  3585.2     .05       0  4283.6     .16       0  4410.9     .05       0
  4447.7     .16       0  4698.4     .05       0  4875.6     .16       0
  4984.2     .07       0  4990.2     .16       0  5104.3     .16       0
  5137.2     .05       0
Bank Sta=4958.9,5029.6
XS Rating Curve= 0 ,0
Exp/Cntr=0.3,0.1

Type RM Length L Ch R = 1 ,129198  ,191,191,191
BEGIN DESCRIPTION:
HURRICANE BAYOU 96.0
END DESCRIPTION:
XS GIS Cut Line= 4
      3821362.68     10486847.64      3820733.35     10488247.36
      3820527.19     10488529.48      3819496.69     10490915.88
#Sta/Elev= 30
    3329  334.85  3354.9  334.87  3605.9  318.65  3696.4  323.35  3714.8  324.77
  3820.6  328.25  3959.7  324.88  4032.2  318.92  4223.1  301.32  4243.7  298.57
  4349.5   292.7  4455.2  293.28    4885  283.83  4940.8  279.51    4947  283.86
    4964   279.2  4998.3  278.02  5003.4  271.65  5026.5  276.07  5029.7  270.29
  5032.5  269.79  5035.7  270.29  5047.4  282.76  5053.6  278.37  5068.3  282.47
  5112.3  275.87  5140.8   284.4  5997.1  284.02  7621.3   308.2  7812.5  306.92
#Mann= 17 ,-1 , 0
    3329     .05       0  3354.9     .16       0  3696.4      .1       0
  3714.8     .08       0  3820.6     .16       0  3959.7     .08       0
  4032.2     .16       0  4223.1     .08       0  4243.7      .1       0
  4349.5     .08       0  4455.2     .05       0    4885     .16       0
    4964     .05       0  4998.3     .16       0  5029.7     .07       0
  5035.7     .16       0  5140.8     .05       0
Bank Sta=4947,5047.4
XS Rating Curve= 0 ,0
Exp/Cntr=0.3,0.1

Type RM Length L Ch R = 1 ,129007  ,1743,1743,1743
BEGIN DESCRIPTION:
HURRICANE BAYOU 95.0
END DESCRIPTION:
XS GIS Cut Line= 4
      3820950.36     10487086.34      3820820.15     10487737.38
      3820060.61     10489039.46      3819084.33     10491219.82
#Sta/Elev= 30
  3677.4  323.58  3682.8  323.65  3782.2  326.36  3873.9  323.72  3961.7  317.57
  4160.6  294.53  4278.7  288.92  4393.6  289.28  4826.9  283.41  4928.5  284.23
    4938  283.92  4987.3  276.57    4993  271.64  5005.8  270.27  5008.5  269.77
  5011.8  270.27  5023.3  274.09  5039.2  282.51  5051.8  283.51  5160.3  282.93
  5233.2  282.84  5382.5  283.25  5443.1  282.72  5939.8  282.93  6386.4  290.45
  6690.4  291.94  6769.4  292.04  7697.2  307.35  7899.2   305.7  8237.7  310.79
#Mann= 17 ,-1 , 0
  3677.4     .05       0  3682.8     .16       0  3782.2     .08       0
  3873.9     .16       0  4278.7     .08       0  4393.6     .05       0
  4826.9     .16       0    4938     .08       0  5005.8     .07       0
  5011.8     .08       0  5023.3     .05       0  5160.3     .08       0
  5233.2     .05       0  5382.5     .08       0  5443.1     .05       0
  6690.4     .08       0  6769.4     .05       0
Bank Sta=4928.5,5051.8
XS Rating Curve= 0 ,0
Exp/Cntr=0.3,0.1

Type RM Length L Ch R = 1 ,127264  ,1463,1463,1463
BEGIN DESCRIPTION:
HURRICANE BAYOU 94.0
END DESCRIPTION:
XS GIS Cut Line= 3
      3820532.96     10485186.04      3819449.61     10487810.19
      3818988.04     10491156.73
#Sta/Elev= 30
  2147.1  344.75  2259.8   348.6  3010.2  315.96  3106.2  315.21  3114.7  313.62
  3187.9  309.47  3507.4  312.65  3990.8  291.87  4885.1  281.36  4953.6  281.79
  4971.4  277.55  4976.8   270.3  4983.4  267.59  5013.4  267.06  5016.1  266.56
  5019.4  267.06  5036.6  274.76  5076.9  281.45    5106  281.11  6044.2  281.31
  6121.1  277.98  6379.1  290.26  6944.4  296.06  7266.7   292.9  7358.7   293.3
    7513  296.91    7540  301.45  7610.7  297.53    7752  303.93  8364.3  310.44
#Mann= 10 ,-1 , 0
  2147.1     .16       0  3010.2     .05       0  3106.2     .08       0
  3114.7     .05       0  4885.1     .16       0  5013.4     .07       0
  5019.4     .16       0    5106     .05       0  7266.7     .12       0
  7358.7     .05       0
Bank Sta=4953.6,5076.9
XS Rating Curve= 0 ,0
Exp/Cntr=0.3,0.1

Type RM Length L Ch R = 1 ,125801  ,1052,1052,1052
BEGIN DESCRIPTION:
HURRICANE BAYOU 93.0
END DESCRIPTION:
XS GIS Cut Line= 3
      3820376.75     10485411.68      3818484.36     10488241.57
      3818744.64     10491694.65
#Sta/Elev= 30
  1796.1  340.59  2160.5  328.84  2289.6  318.98  2336.8  319.75  2520.8  323.67
  2852.9  312.88  2902.2  308.13  3010.3  303.03    3695   283.4  4223.4  278.56
  4887.8  278.67  4929.1  278.93  4958.2  276.07  4971.2  272.36  4980.2  266.82
  4991.3   264.7    4994   264.2  4997.3   264.7  5022.2  278.98  5043.2  279.82
  5059.4  279.18  5467.3   277.6  5660.3  284.74  6683.2  289.12  7605.8  303.19
  7863.1  312.19  7986.9  313.69  8067.2  310.81  8633.8  313.18  8663.3  313.35
#Mann= 7 ,-1 , 0
  1796.1     .16       0  2336.8     .05       0  4887.8     .16       0
  4991.3     .07       0  4997.3     .16       0  5059.4     .05       0
  8633.8      .1       0
Bank Sta=4929.1,5043.2
XS Rating Curve= 0 ,0
Exp/Cntr=0.3,0.1

Type RM Length L Ch R = 1 ,124749  ,581,581,581
BEGIN DESCRIPTION:
HURRICANE BAYOU 92.0
END DESCRIPTION:
XS GIS Cut Line= 4
      3819298.53     10485553.12      3817683.94     10487831.78
      3817384.46     10488704.17      3816538.11     10490683.33
#Sta/Elev= 30
  2498.1  323.83  2939.6  311.11  3649.6  279.65  4868.1  277.53  4947.8  278.48
  4962.5  275.57  4980.4  263.18  4983.2  262.68  4986.4  263.18  5006.9  265.71
  5019.2  275.61  5033.9  277.84    5310  274.89  5458.3  277.32  5473.8  274.77
  5479.4  267.42  5505.1  265.86  5531.1  276.01  5574.6  277.02  5585.2   267.2
  5598.9  266.82  5631.3  276.98  5656.1   276.4  5680.3  266.78  5687.4  274.02
  5706.1  278.46  6442.1  278.43  6451.9  278.49  7532.8  288.36  8365.7  312.27
#Mann= 9 ,-1 , 0
  2498.1     .05       0  4868.1     .16       0  4980.4     .07       0
  4986.4     .16       0    5310     .12       0  5631.3     .16       0
  5706.1     .05       0  6442.1     .16       0  6451.9     .05       0
Bank Sta=4947.8,5033.9
XS Rating Curve= 0 ,0
Exp/Cntr=0.3,0.1

Type RM Length L Ch R = 1 ,124168  ,809,809,809
BEGIN DESCRIPTION:
HURRICANE BAYOU 91.0
END DESCRIPTION:
XS GIS Cut Line= 4
       3818777.7     10485631.25      3817631.86     10487063.55
      3817111.02     10488769.28      3816121.46     10490631.23
#Sta/Elev= 30
  2651.9  321.07  2813.8  315.34  3084.3   292.2  3503.7  280.69  4100.8  274.15
  4732.1  276.94  4838.1  272.31  4957.2  277.55  4995.3  262.98  5012.9  262.58
  5015.6  262.08  5018.9  262.58  5036.8  273.79  5056.4   273.3  5088.5  266.59
  5099.5  276.33    5110   277.5  5319.1  276.38    5340  264.22  5371.8  265.38
  5392.3  275.71  5423.7  264.91  5437.4  269.06    5455  265.79  5475.9  277.46
  5502.1  277.15    5515  276.58  6916.1  282.93  7394.4  297.24  8378.2  310.18
#Mann= 7 ,-1 , 0
  2651.9     .05       0  4732.1     .16       0  5012.9     .07       0
  5018.9     .16       0  5056.4     .12       0  5502.1     .16       0
    5515     .05       0
Bank Sta=4957.2,5110
XS Rating Curve= 0 ,0
Exp/Cntr=0.3,0.1

Type RM Length L Ch R = 1 ,123359  ,281,281,281
BEGIN DESCRIPTION:
HURRICANE BAYOU 90.0
END DESCRIPTION:
XS GIS Cut Line= 3
      3818048.52     10485396.89      3816850.61     10487766.67
      3815392.28     10490592.18
#Sta/Elev= 30
  2742.6  319.08  2996.8  316.71  3152.8  308.36  3192.3  302.35  3368.9  287.08
  3548.4  277.78  3988.5  272.66  4023.7  275.23  4902.5  275.18  4941.3  277.65
  4963.6  274.41  4969.2  267.36  4976.1  264.33  4995.5   261.8  4998.3   261.3
  5001.5   261.8  5030.5  266.79  5036.1  274.66  5052.8  276.19  5102.2  275.62
  5514.4  272.76  6358.4  280.39    6849  292.65  7026.2  293.36  7397.3  306.25
  7821.4  308.11  7917.7  306.17  8147.7   310.1  8316.5  307.57  8577.6  308.48
#Mann= 7 ,-1 , 0
  2742.6     .05       0  3192.3     .16       0  3368.9     .05       0
  4902.5     .16       0  4995.5     .07       0  5001.5     .16       0
  5102.2     .05       0
Bank Sta=4941.3,5052.8
XS Rating Curve= 0 ,0
Exp/Cntr=0.3,0.1

Type RM Length L Ch R = 1 ,123078  ,635,635,635
BEGIN DESCRIPTION:
HURRICANE BAYOU 89.0
END DESCRIPTION:
XS GIS Cut Line= 3
      3817449.59     10485660.22      3816799.61     10487260.19
      3815399.63     10489460.16
#Sta/Elev= 30
  3273.3  316.32  3359.6  311.78  3402.8  306.24  3424.8  306.45  3662.4  280.95
  3748.2  275.35  3964.1   274.7  3996.4   271.9  4032.3  274.21  4622.5  272.22
  4850.3  275.27    4956  276.23  4967.9  273.32  4987.9  261.22  4990.7  260.72
  4993.9  261.22  5003.2  262.06  5013.8  267.41  5059.5  275.56  5070.5   275.3
  5247.5  275.31  5420.2  271.25  5529.4  273.47  5926.5  272.87    6327  283.75
  6426.9  281.31  6739.3  289.39  7303.1   294.8  7360.7  298.65  7607.9  307.95
#Mann= 7 ,-1 , 0
  3273.3     .05       0  3424.8     .16       0  3662.4     .05       0
  4850.3     .16       0  4987.9     .07       0  4993.9     .16       0
  5070.5     .05       0
Bank Sta=4956,5059.5
XS Rating Curve= 0 ,0
Exp/Cntr=0.3,0.1

Type RM Length L Ch R = 1 ,122443  ,601,601,601
BEGIN DESCRIPTION:
HURRICANE BAYOU 88.0
END DESCRIPTION:
XS GIS Cut Line= 3
      3817199.63     10485560.16      3816399.61     10486860.19
      3815199.59     10489260.23
#Sta/Elev= 30
    3452  315.59    3539  314.45  3654.9  309.26  3902.3  290.11  3975.6  278.86
  4112.9     273  4127.2   270.7  4244.2  273.33  4426.6  271.85  4892.6  274.09
  4949.5  275.26  4970.8  271.99  4975.5  267.16  4981.3  267.16  4986.9  262.38
  4997.8  261.07  5000.6  260.57  5003.8  261.07  5014.8   261.2  5031.6  272.77
  5045.6  275.01  5105.4  273.89  5626.9  271.31  5775.1  272.57  5791.8   270.4
  6468.3  274.04  6856.8  280.11  7035.7  289.34    7385  292.03  7661.8   305.5
#Mann= 5 ,-1 , 0
    3452     .05       0  4892.6     .16       0  4997.8     .07       0
  5003.8     .16       0  5105.4     .05       0
Bank Sta=4949.5,5045.6
XS Rating Curve= 0 ,0
Exp/Cntr=0.3,0.1

Type RM Length L Ch R = 1 ,121842  ,568,568,568
BEGIN DESCRIPTION:
HURRICANE BAYOU 87.0
END DESCRIPTION:
XS GIS Cut Line= 3
      3817601.01     10485019.35      3816099.61     10486610.19
      3814699.63     10489010.15
#Sta/Elev= 30
  2812.6  316.48  3139.7  316.82  3408.3  310.66  3599.3   315.4  3903.5  294.37
  4073.4  277.79    4236     269  4278.5  272.88  4412.8  268.87  4448.4  271.96
  4890.7  273.61  4964.7  274.63  4978.8  270.79  4986.1  262.81  4993.6  260.41
  4996.4  259.91  4999.6  260.41  5013.7  260.67  5023.2  264.89  5029.4  273.15
  5153.3  273.56  5694.7  270.18  6119.3  271.59  6156.5  267.98  6418.7  273.93
  6819.7   272.1  7097.6  281.31  7273.7   280.1  7646.2  291.19  7778.5  298.56
#Mann= 6 ,-1 , 0
  2812.6     .05       0  4890.7     .16       0  4993.6     .07       0
  4999.6     .16       0  5153.3     .05       0  7646.2     .16       0
Bank Sta=4964.7,5029.4
XS Rating Curve= 0 ,0
Exp/Cntr=0.3,0.1

Type RM Length L Ch R = 1 ,121274  ,689,689,689
BEGIN DESCRIPTION:
HURRICANE BAYOU 86.0
END DESCRIPTION:
XS GIS Cut Line= 3
      3815647.92      10484563.6      3815599.61     10486460.19
       3814199.6     10489560.22
#Sta/Elev= 30
  3108.7  316.15  3177.4  317.16  3275.5   319.5  3373.5  320.63  3519.3  312.33
    3522  311.99  3681.4  295.79    3854  279.01  4145.6  269.69  4270.9  270.93
    4449  268.74  4867.8  273.06  4965.9  273.52  4985.9  264.96  5014.7  265.21
  5017.2  260.98    5020  260.48  5023.2  260.98  5027.8  268.29  5043.3  268.72
  5049.8  275.02  5093.7  272.85  6282.8  271.46  6311.6  267.28    7610  280.48
  7901.1  298.91  8006.9  303.96  8112.8  310.01  8138.8  310.68  8407.4     317
#Mann= 19 ,-1 , 0
  3108.7     .15       0  3177.4      .1       0  3275.5     .08       0
  3373.5     .05       0  3519.3     .08       0    3522     .05       0
  3681.4     .16       0    3854     .05       0  4270.9     .16       0
    4449     .05       0  4867.8     .16       0  5017.2     .07       0
  5023.2     .16       0  5093.7     .05       0    7610     .16       0
  7901.1     .08       0  8006.9     .16       0  8112.8     .08       0
  8138.8     .05       0
Bank Sta=4965.9,5049.8
XS Rating Curve= 0 ,0
Exp/Cntr=0.3,0.1

Type RM Length L Ch R = 1 ,120585  ,614,614,614
BEGIN DESCRIPTION:
HURRICANE BAYOU 85.0
END DESCRIPTION:
XS GIS Cut Line= 3
      3815449.61     10484910.16      3815249.61     10486510.19
      3814149.61     10489310.19
#Sta/Elev= 30
  3395.7  322.58  3486.4  322.09  3514.1  317.21  3680.4  305.73  3917.3  282.95
  4159.1  270.01  4353.1  268.12  4878.3  271.62  4957.8  273.13  4970.4  270.66
    4988  259.31  4995.1  259.05  4997.9  258.55  5001.1  259.05  5029.7  272.49
  5163.4   271.8  5600.3  267.37    6233  270.47  6265.2  266.88  6310.4  270.56
  6780.9  270.64  7221.4  279.13  7242.9  275.78  7267.1   279.7  7307.4  277.91
  7315.9  281.98  7366.8  282.58  7562.6  297.92  7829.1  307.15  8016.5  311.61
#Mann= 7 ,-1 , 0
  3395.7     .05       0  4878.3     .16       0  4995.1     .07       0
  5001.1     .16       0  5163.4     .05       0  7366.8     .16       0
  7829.1     .05       0
Bank Sta=4957.8,5029.7
XS Rating Curve= 0 ,0
Exp/Cntr=0.3,0.1

Type RM Length L Ch R = 1 ,119971  ,1274,1274,1274
BEGIN DESCRIPTION:
HURRICANE BAYOU 84.0
END DESCRIPTION:
XS GIS Cut Line= 3
      3815299.62     10485110.16      3814799.61     10486710.19
      3813147.91     10489251.09
#Sta/Elev= 30
  3318.6  313.77  3350.1  308.13  3360.5  309.67  3372.6  303.95  3437.5  307.25
  3517.7  294.76  3685.3  282.45  3875.5  270.85  4010.6  269.83  4031.1   266.1
  4083.4  270.02  4863.4  267.99  4946.2  272.05  4963.5  268.54  4981.5  258.44
  4984.2  257.94  4987.5  258.44  5008.5  260.46  5017.6  270.43  5023.6  266.29
  5038.7  271.59  5111.4  271.75  5805.7  266.16  6512.2  269.04  6678.2  275.77
  6867.5  296.07  7010.6  304.46  7249.2  311.06  7880.8  313.53  8025.5  313.07
#Mann= 6 ,-1 , 0
  3318.6     .05       0  4863.4     .16       0  4981.5     .07       0
  4987.5     .16       0  5111.4     .05       0  7880.8     .16       0
Bank Sta=4946.2,5038.7
XS Rating Curve= 0 ,0
Exp/Cntr=0.3,0.1

Type RM Length L Ch R = 1 ,118697  ,536,536,536
BEGIN DESCRIPTION:
HURRICANE BAYOU 83.0
END DESCRIPTION:
XS GIS Cut Line= 2
      3814918.74     10484576.62        3812588.     10488821.43
#Sta/Elev= 30
  3318.1  321.89  3379.5  321.17  3617.8  312.75  3696.8   308.4  3792.8  296.42
  3843.7  295.24  3887.3  286.31  4115.6   268.5  4930.3  269.92  4947.6  269.72
  4985.5  258.27  4996.2  257.96  4998.9  257.46  5002.2  257.96  5007.3  265.02
    5013  261.92  5029.1   271.2  5097.5   268.9  6345.4  264.44  6605.8  266.86
  6812.3   278.9  7077.2  302.22  7142.8  303.83  7186.8  299.95  7236.9  298.37
  7290.8  289.91    7378  301.01  7465.2  307.58  7851.7  309.46  8160.7  312.62
#Mann= 12 ,-1 , 0
  3318.1     .08       0  3379.5     .05       0  3617.8     .16       0
  3792.8     .05       0  4930.3     .16       0  4996.2     .07       0
  5002.2     .16       0  5097.5     .05       0  7077.2     .08       0
  7142.8     .05       0  7186.8     .16       0  7851.7     .05       0
#XS Ineff= 1 ,-1
  7142.8  7415.4   304.2
Permanent Ineff=
       F
Bank Sta=4947.6,5029.1
XS Rating Curve= 0 ,0
Exp/Cntr=0.3,0.1

Type RM Length L Ch R = 1 ,118161  ,194,194,194
BEGIN DESCRIPTION:
HURRICANE BAYOU 82.0
END DESCRIPTION:
XS GIS Cut Line= 4
      3814710.42     10484277.13      3813811.98     10485579.21
      3813317.19     10486516.71      3812301.55     10488521.95
#Sta/Elev= 30
  2966.4  316.59    2986  316.67    2996  316.71  3112.2  315.04  3139.4  315.07
  3573.4  301.54  3803.3   282.2  4081.3  268.02  4895.2  267.49  4943.8  268.13
  4966.7  269.04  4979.1  256.66  4985.7  256.57  4988.5  256.07  4991.7  256.57
  5024.4  269.39  5123.5  267.64  5161.3  267.34  5351.8  265.98  5378.9  266.12
    5580  265.46  5596.4  265.62  6317.6  267.72  6479.2  275.44  6645.4   292.8
  6779.3  295.62  6953.3  301.05    7124  307.92  7587.3  304.82  7856.2  309.27
#Mann= 20 ,-1 , 0
  2966.4     .15       0    2986      .1       0    2996     .08       0
  3112.2     .05       0  3139.4     .08       0  4081.3     .05       0
  4895.2     .08       0  4943.8     .05       0  4985.7     .03       0
  4991.7     .05       0  5123.5     .08       0  5161.3     .05       0
  5351.8     .08       0  5378.9     .05       0    5580     .08       0
  5596.4     .05       0  6645.4     .08       0  6779.3     .05       0
  6953.3     .08       0    7124     .05       0
Bank Sta=4966.7,5024.4
XS Rating Curve= 0 ,0
Exp/Cntr=0.3,0.1

Type RM Length L Ch R = 1 ,117967  ,919,919,919
BEGIN DESCRIPTION:
HURRICANE BAYOU 81.0
END DESCRIPTION:
XS GIS Cut Line= 4
      3814528.15     10484172.93      3813642.71     10485396.92
      3813291.15     10486217.23      3812015.09     10488469.86
#Sta/Elev= 30
  2922.5  311.38  2946.3   311.2  3069.4  306.61  3187.2  302.83  3318.2   299.6
  3422.9  294.56  3542.6  290.55  4093.3  275.37  4215.1  267.21  4962.9  268.59
  4983.5   255.8  4986.3   255.3  4989.5   255.8  5002.5  256.09  5010.1  265.05
  5024.2   268.7  5428.4  266.95  5432.4  267.35  6004.9  263.01    6318  269.11
  7060.2  308.16  7152.6     308  7187.6  308.76  7335.2  308.36  7535.3  307.99
  7582.7  309.07  7667.3  303.59  7783.2   306.1    7846  312.61  7914.6  312.11
#Mann= 19 ,-1 , 0
  2922.5     .08       0  2946.3      .1       0  3069.4     .15       0
  3187.2     .08       0  3318.2     .05       0  3422.9     .08       0
  3542.6     .05       0  4983.5     .03       0  4989.5     .05       0
  5428.4     .08       0  5432.4     .05       0  7060.2     .08       0
  7152.6     .05       0  7187.6     .16       0  7335.2     .08       0
  7535.3     .16       0  7582.7     .05       0  7667.3     .16       0
  7783.2     .05       0
Bank Sta=4962.9,5024.2
XS Rating Curve= 0 ,0
Exp/Cntr=0.3,0.1

Type RM Length L Ch R = 1 ,117048  ,506,506,506
BEGIN DESCRIPTION:
HURRICANE BAYOU 80.0
END DESCRIPTION:
XS GIS Cut Line= 4
      3814397.95     10484003.66       3812952.6     10485409.94
      3812353.65       10486699.       3812184.5     10488013.15
#Sta/Elev= 30
  2305.8  304.88  2426.1  303.47  2430.4  303.23  2565.8  297.28  2569.3  297.32
  2938.6  283.31  3327.5  274.24  3695.3  265.73  4528.9   264.8  4973.2  268.37
  4980.4  264.15  4985.9  266.31  4995.3  258.36  5005.8  256.05  5008.6  255.55
  5011.8  256.05  5039.4  267.28    5192  266.51  5197.5     259  5204.8  258.87
  5237.8  266.83  5689.3   266.1  5886.2  269.53  6158.4  280.22  6420.5  293.07
  6450.8  291.64  6571.8  299.54  6662.7  300.93  6702.8  306.12  7068.8  308.21
#Mann= 10 ,-1 , 0
  2305.8     .05       0  2426.1     .08       0  2430.4      .1       0
  2565.8     .08       0  2569.3     .05       0  3327.5     .16       0
  5005.8     .07       0  5011.8     .16       0  6158.4     .05       0
  6662.7     .16       0
#XS Ineff= 2 , 0
         4113.64  278.75 5354.55          277.07
Permanent Ineff=
       F       F
Bank Sta=4973.2,5039.4
XS Rating Curve= 0 ,0
Exp/Cntr=0.3,0.1

Type RM Length L Ch R = 1 ,116542  ,313,313,313
BEGIN DESCRIPTION:
HURRICANE BAYOU 79.0
END DESCRIPTION:
XS GIS Cut Line= 5
      3814111.43     10483521.93      3812926.56     10483899.52
      3812379.69     10485422.96      3812236.46     10486060.98
      3812184.37      10487792.8
#Sta/Elev= 30
  1734.3  303.48    1974  303.12  2187.5  297.71    2261  288.05  2418.4  284.58
  2639.2  265.45  2680.8   266.4  2698.3  269.63  2832.4  265.06  4053.1  265.37
  4381.1  262.61  4487.3  265.46  4737.1  264.36  4962.6  267.15  4972.9  260.98
  4986.3  255.96  4989.6  256.46  5029.9   266.6  5329.6  264.67  5439.7  271.76
  5609.8  275.34  5739.8  270.43  5969.9  271.77  6610.2  295.28  6643.9  293.35
  6700.3  296.39  6730.3  294.76  6790.3   298.1  6800.3  301.12    6983  307.34
#Mann= 4 ,-1 , 0
  1734.3     .16       0  4972.9     .07       0  4989.6     .16       0
    6983     .16       0
#XS Ineff= 2 , 0
         3117.05  285.59 5039.77          275.17
Permanent Ineff=
       F       F
Bank Sta=4962.6,5029.9
XS Rating Curve= 0 ,0
Exp/Cntr=0.3,0.1

Type RM Length L Ch R = 1 ,116229  ,282,282,282
BEGIN DESCRIPTION:
HURRICANE BAYOU 78.0
END DESCRIPTION:
XS GIS Cut Line= 5
      3814990.44     10480897.42      3813065.13     10482755.75
      3812353.32     10484596.03      3811980.06     10485819.99
      3811971.38     10488363.36
#Sta/Elev= 30
  -768.1  311.27  -567.6  316.88   -44.2  317.34   146.8  311.54   302.5  298.92
   514.4  299.15   761.9  276.71   832.7  274.16  1561.2  268.69  1674.4  276.22
  1794.5  267.77  1900.8  271.22  3099.2  263.39  4566.1  265.66  4593.7  260.63
  4664.5  261.49  4697.4  265.98  4942.8  267.63  4975.6  265.56  4993.4  254.65
  5008.2  253.88  5011.5  254.38  5014.4  264.79    5036  267.42  5180.7  263.79
  5530.7  266.96  5910.7  284.08  6230.7  286.69  6580.7  303.18  7703.9  310.98
#Mann= 5 ,-1 , 0
  -768.1     .16       0  1674.4     .16       0  4993.4     .07       0
  5014.4     .16       0  7703.9     .05       0
#XS Ineff= 2 , 0
         4261.36  275.82 5056.82          277.24
Permanent Ineff=
       F       F
Bank Sta=4942.8,5036
XS Rating Curve= 0 ,0
Exp/Cntr=0.3,0.1
