--- SIMS BRANCH.prj (project) ---

Proj Title=SIMS BRANCH Base Level Engineering
Current Plan=p01
Default Exp/Contr=0.3,0.1
English Units
Geom File=g01
Flow File=f01
Plan File=p01
BEGIN DESCRIPTION:
SIMS BRANCH
END DESCRIPTION:

--- SIMS BRANCH.p01 (plan) ---

Plan Title=Multiple Run
Short Identifier=Multiple
Geom File=g01
Flow File=f01
Subcritical Flow
K Sum by GR= 0
Std Step Tol= 0.01
Critical Tol= 0.01
Num of Std Step Trials= 20
Max Error Tol= 0.3
Flow Tol Ratio= 0.001
Split Flow NTrial= 30
Split Flow Tol= 0.02
Split Flow Ratio= 0.02
Log Output Level= 0
Friction Slope Method= 1
Unsteady Friction Slope Method= 2
Unsteady Bridges Friction Slope Method= 1
Parabolic Critical Depth
Global Vel Dist=  1 , 1 , 1
Global Log Level= 0
CheckData=True
Encroach Param= -1, 0, 0, 0
BEGIN DESCRIPTION:
Multiple Run
END DESCRIPTION:

--- SIMS BRANCH.f01 (steady flow) ---

Flow Title=Multiple
Number of Profiles=7
Profile Names=10-year,25-year,50-year,1pct_min,100-year,1pct_plu,500-year
River Rch & RM= SIMS BRANCH,Reach-1,22887
     620     838    1019     911    1232    1666    1806
River Rch & RM= SIMS BRANCH,Reach-1,18023
     782    1067    1305    1171    1583    2141    2340
River Rch & RM= SIMS BRANCH,Reach-1,12795
     944    1297    1591    1431    1936    2618    2878
River Rch & RM= SIMS BRANCH,Reach-1,3924
    1021    1407    1731    1561    2112    2856    3155
Boundary for River Rch & Prof#=SIMS BRANCH,Reach-1,1
Up Type=0
Dn Type=3
Dn Slope=0.005
Boundary for River Rch & Prof#=SIMS BRANCH,Reach-1,2
Up Type=0
Dn Type=3
Dn Slope=0.005
Boundary for River Rch & Prof#=SIMS BRANCH,Reach-1,3
Up Type=0
Dn Type=3
Dn Slope=0.005
Boundary for River Rch & Prof#=SIMS BRANCH,Reach-1,4
Up Type=0
Dn Type=3
Dn Slope=0.005
Boundary for River Rch & Prof#=SIMS BRANCH,Reach-1,5
Up Type=0
Dn Type=3
Dn Slope=0.005
Boundary for River Rch & Prof#=SIMS BRANCH,Reach-1,6
Up Type=0
Dn Type=3
Dn Slope=0.005
Boundary for River Rch & Prof#=SIMS BRANCH,Reach-1,7
Up Type=0
Dn Type=3
Dn Slope=0.005

--- SIMS BRANCH.g01 (geometry) ---

Geom Title=Existing Conditions

River Reach=SIMS BRANCH,Reach-1
Reach XY= 30
      3814249.61     10509510.19      3814444.00     10508837.00
      3814323.50     10508321.00      3814524.50     10507845.00
      3814175.75     10506634.00      3814370.00     10506276.00
      3813968.50     10505114.00      3814567.75     10504708.00
      3814256.25     10503680.00      3814519.75     10503001.00
      3814144.75     10502883.00      3814135.25     10502247.00
      3813651.75     10501715.00      3814025.75     10501126.00
      3813421.25     10500454.00      3813539.75     10499651.00
      3814025.75     10499464.00      3814408.50     10498108.00
      3814297.50     10497694.00      3814550.25     10497621.00
      3814966.25     10496993.00      3815102.25     10497046.00
      3815637.75     10496495.00      3815730.00     10495817.00
      3816142.25     10495632.00      3816823.50     10494428.00
      3816875.25     10493973.00      3817242.25     10494035.00
      3817265.25     10493679.00      3817849.00     10493261.00

Type RM Length L Ch R = 1,22887,538,538,538
BEGIN DESCRIPTION:
SIMS BRANCH 46.0
END DESCRIPTION:
XS GIS Cut Line= 3
      3814599.62     10509360.20      3814299.61     10509110.19
      3813699.60     10508960.19
#Sta/Elev= 30
  4628.7  402.45  4635.9  401.48  4671.0  400.57  4678.8  398.93  4699.7  398.68
  4714.0  397.30  4777.8  395.98  4784.9  394.99  4835.3  393.01  4941.1  388.88
  4997.7  388.03  5012.1  388.84  5017.7  388.15  5042.4  388.30  5072.3  387.16
  5075.5  386.89  5078.2  386.39  5081.5  386.89  5173.8  390.52  5248.6  392.00
  5266.6  393.62  5289.8  394.14  5318.1  395.98  5325.9  397.25  5349.1  398.08
  5421.2  404.00  5483.1  407.43  5503.7  409.63  5524.3  409.47  5637.7  414.52
#Mann=6,-1,0
  4628.7    0.16       0  4835.3    0.12       0  5017.7    0.07       0
  5072.3    0.05       0  5075.5    0.07       0  5081.5    0.05       0
Bank Sta=5075.5,5081.5
Exp/Cntr=0.3,0.1

Type RM Length L Ch R = 1,22349,42,42,42
BEGIN DESCRIPTION:
Mapping XS 5a46fbbe
END DESCRIPTION:
XS GIS Cut Line= 6
      3815167.29     10509404.75      3814476.33     10508675.60
      3814455.50     10508623.52      3814396.47     10508623.52
      3814344.39     10508668.66      3813512.81     10508824.58
#Sta/Elev= 30
  3907.0  432.88  3972.2  430.05  3979.5  428.55  4096.8  421.96  4156.3  419.08
  4170.4  416.42  4311.6  407.67  4630.1  392.85  4715.0  391.33  4743.4  389.20
  4854.2  386.50  4884.8  386.47  4899.0  387.94  4911.7  387.45  4914.2  385.91
  4919.6  385.57  5090.6  385.36  5099.8  387.26  5125.0  388.64  5137.8  387.74
  5142.4  384.93  5145.1  384.43  5148.4  384.93  5348.1  392.35  5521.8  400.85
  5552.4  403.38  5613.4  403.70  5664.3  407.71  5841.5  417.87  5945.9  426.47
#Mann=4,-1,0
  3907.0    0.16       0  4096.8    0.05       0  5142.4    0.03       0
  5148.4    0.05       0
Bank Sta=5142.4,5148.4
Exp/Cntr=0.3,0.1

Type RM Length L Ch R = 1,22307,31,31,31
BEGIN DESCRIPTION:
SIMS BRANCH 45.0
END DESCRIPTION:
XS GIS Cut Line= 6
      3815222.89     10509415.22      3814462.44     10508585.32
      3814406.89     10508581.85      3814365.22     10508595.74
      3814313.14     10508647.82      3813469.41     10508745.04
#Sta/Elev= 30
  3830.1  434.10  3970.7  426.16  4023.2  424.39  4189.6  412.91  4352.4  403.99
  4614.6  392.75  4826.7  386.99  4890.9  387.00  4897.7  388.68  4911.9  387.80
  4933.1  388.82  4940.2  387.83  4947.3  389.35  5023.2  389.91  5054.5  389.04
  5070.1  389.84  5076.2  388.23  5100.8  389.67  5121.5  389.12  5141.1  385.29
  5143.9  384.79  5147.1  385.29  5295.1  389.38  5345.4  391.98  5370.1  391.92
  5506.5  400.73  5577.0  402.17  5667.5  408.10  5798.4  413.70  5979.8  428.25
#Mann=4,-1,0
  3830.1    0.16       0  4023.2    0.05       0  5141.1    0.03       0
  5147.1    0.05       0
Bank Sta=5141.1,5147.1
Exp/Cntr=0.3,0.1

Type RM Length L Ch R = 1,22276,222,222,222
BEGIN DESCRIPTION:
Mapping XS 6addd53a
END DESCRIPTION:
XS GIS Cut Line= 6
      3815295.81     10509387.44      3814504.11     10508574.91
      3814469.39     10508543.66      3814347.86     10508561.02
      3814271.47     10508602.68      3813469.39     10508682.55
#Sta/Elev= 30
  3763.4  433.75  3836.6  428.90  3906.0  426.09  3935.6  424.42  3978.0  424.01
  4006.3  420.97  4048.7  419.93  4133.6  414.22  4310.4  404.65  4557.8  394.01
  4741.7  388.38  4869.0  385.93  4957.5  386.94  5015.1  385.14  5055.5  385.72
  5073.5  384.48  5079.2  385.57  5092.4  384.22  5095.1  383.72  5098.4  384.22
  5110.9  385.72  5236.6  387.89  5457.7  399.34  5568.2  402.93  5628.5  406.29
  5638.6  408.22  5648.6  407.41  5689.1  408.34  5809.4  415.24  5960.4  426.98
#Mann=4,-1,0
  3763.4    0.16       0  3906.0    0.05       0  5092.4    0.03       0
  5098.4    0.05       0
Bank Sta=5092.4,5098.4
Exp/Cntr=0.3,0.1

Type RM Length L Ch R = 1,22054,597,597,597
BEGIN DESCRIPTION:
SIMS BRANCH 44.0
END DESCRIPTION:
XS GIS Cut Line= 4
      3815105.62     10508642.74      3814699.84     10508382.35
      3814098.72     10508334.61      3813523.04     10508527.22
#Sta/Elev= 30
  4146.7  400.13  4341.9  393.23  4355.8  392.08  4399.4  391.89  4405.3  391.02
  4450.9  390.44  4462.8  389.48  4493.2  389.79  4499.2  388.97  4550.7  387.48
  4571.8  387.83  4669.2  385.83  4779.5  385.90  4809.6  384.02  4829.7  384.52
  4889.9  383.41  4920.0  384.35  4927.0  383.01  4929.8  382.51  4933.0  383.01
  4950.1  384.14  5000.2  383.10  5060.4  384.14  5080.5  385.48  5329.7  394.88
  5399.6  399.46  5462.9  400.56  5577.0  404.84  5740.1  413.51  5838.9  420.44
#Mann=3,-1,0
  4146.7    0.05       0  4927.0    0.03       0  4933.0    0.05       0
Bank Sta=4927,4933
Exp/Cntr=0.3,0.1

Type RM Length L Ch R = 1,21457,616,616,616
BEGIN DESCRIPTION:
SIMS BRANCH 43.0
END DESCRIPTION:
XS GIS Cut Line= 3
      3815099.64     10508460.22      3814499.61     10507860.19
      3813899.66     10507910.18
#Sta/Elev= 30
  4162.5  394.61  4176.7  393.78  4205.0  393.81  4275.7  389.50  4289.8  390.61
  4403.0  387.67  4558.5  384.87  4643.4  384.41  4671.7  385.18  4699.9  383.99
  4770.7  382.83  4912.1  382.07  4926.2  381.14  4993.9  380.56  4996.7  380.06
  4999.9  380.56  5051.2  380.60  5091.3  382.51  5211.8  381.53  5292.0  383.63
  5392.4  388.65  5412.5  392.03  5462.6  396.23  5512.8  399.07  5532.9  399.14
  5550.4  400.53  5555.4  401.74  5573.0  400.93  5583.0  402.52  5613.1  404.32
#Mann=3,-1,0
  4162.5    0.05       0  4993.9    0.03       0  4999.9    0.05       0
Bank Sta=4993.9,4999.9
Exp/Cntr=0.3,0.1

Type RM Length L Ch R = 1,20841,355,355,355
BEGIN DESCRIPTION:
SIMS BRANCH 42.0
END DESCRIPTION:
XS GIS Cut Line= 3
      3815452.91     10507475.24      3814543.59     10507282.09
      3813801.02     10507843.98
#Sta/Elev= 30
  3854.5  389.36  3990.8  385.91  4002.6  385.01  4399.7  383.02  4433.9  381.59
  4491.7  380.52  4577.6  380.67  4604.2  379.28  4771.0  378.06  4927.6  378.63
  4956.7  378.98  4977.5  380.26  5003.6  377.76  5006.4  377.26  5009.6  377.76
  5014.8  379.60  5027.4  380.24  5056.6  378.69  5085.7  379.69  5106.5  378.46
  5171.0  378.61  5314.5  382.51  5464.4  389.41  5514.3  392.17  5520.6  393.42
  5549.7  395.20  5564.2  395.28  5570.5  396.28  5620.4  399.08  5715.3  402.68
#Mann=3,-1,0
  3854.5    0.05       0  5003.6    0.03       0  5009.6    0.05       0
Bank Sta=5003.6,5009.6
Exp/Cntr=0.3,0.1

Type RM Length L Ch R = 1,20486,447,447,447
BEGIN DESCRIPTION:
SIMS BRANCH 41.0
END DESCRIPTION:
XS GIS Cut Line= 3
      3815249.65     10506610.17      3814349.61     10507060.19
      3813899.59     10507660.21
#Sta/Elev= 30
  3973.3  395.86  3986.0  395.01  4160.6  387.29  4317.1  382.25  4398.2  381.75
  4510.0  378.49  4591.1  378.16  4652.5  379.60  4733.6  378.60  4742.0  377.21
  4756.0  378.38  4786.7  377.96  4792.3  379.43  4902.4  377.32  4948.8  377.00
  4986.9  378.60  4990.1  376.45  4992.9  375.95  4996.1  376.45  5007.7  378.57
  5036.9  379.78  5063.8  379.20  5093.1  379.65  5122.3  377.80  5229.6  379.02
  5419.0  378.68  5536.9  380.92  5634.2  385.59  5693.1  390.14  5729.6  391.51
#Mann=8,-1,0
  3973.3    0.16       0  3986.0    0.05       0  4902.4    0.16       0
  4990.1    0.07       0  4996.1    0.16       0  5063.8    0.05       0
  5419.0    0.16       0  5634.2    0.05       0
Bank Sta=4990.1,4996.1
Exp/Cntr=0.3,0.1

Type RM Length L Ch R = 1,20039,497,497,497
BEGIN DESCRIPTION:
SIMS BRANCH 40.0
END DESCRIPTION:
XS GIS Cut Line= 3
      3815099.59     10506510.19      3814199.61     10506660.19
      3813299.60     10507560.20
#Sta/Elev= 30
  4068.6  389.06  4200.4  385.68  4284.0  382.12  4453.8  378.87  4494.4  377.13
  4595.8  377.76  4772.2  376.16  4849.2  375.16  4920.2  375.89  4970.9  377.84
  4984.5  377.54  4992.1  374.42  4994.9  373.92  4998.1  374.42  5023.4  377.73
  5051.7  376.23  5108.3  375.76  5150.7  377.06  5179.0  375.97  5229.1  376.58
  5391.1  379.05  5447.7  377.83  5518.4  377.65  5879.6  384.33  5985.1  386.81
  5999.2  387.87  6055.8  388.55  6098.2  390.78  6126.5  390.70  6253.8  396.06
#Mann=6,-1,0
  4068.6    0.05       0  4772.2    0.16       0  4992.1    0.07       0
  4998.1    0.16       0  5229.1    0.05       0  5879.6    0.16       0
Bank Sta=4992.1,4998.1
Exp/Cntr=0.3,0.1

Type RM Length L Ch R = 1,19542,518,518,518
BEGIN DESCRIPTION:
SIMS BRANCH 39.0
END DESCRIPTION:
XS GIS Cut Line= 3
      3815208.06     10506367.11      3814096.99     10506235.17
      3812395.62     10507179.61
#Sta/Elev= 30
  4151.9  392.23  4563.2  380.49  4754.6  376.37  4836.3  376.11  4895.5  376.26
  4936.1  375.00  4945.9  372.76  4966.0  374.80  4986.2  374.79  4993.2  370.49
  4996.0  369.99  4999.2  370.49  5013.8  374.25  5018.8  372.54  5036.5  374.95
  5066.7  374.25  5096.5  375.51  5258.1  373.23  5347.7  373.50  5396.9  375.25
  5508.0  372.89  5588.0  375.66  5646.3  373.87  5882.3  377.16  6112.0  377.79
  6434.4  381.63  6766.1  387.90  7082.3  395.08  7147.5  397.82  7216.7  397.87
#Mann=5,-1,0
  4151.9    0.05       0  4836.3    0.16       0  4993.2    0.07       0
  4999.2    0.16       0  5882.3    0.05       0
Bank Sta=4993.2,4999.2
Exp/Cntr=0.3,0.1

Type RM Length L Ch R = 1,19024,1001,1001,1001
BEGIN DESCRIPTION:
SIMS BRANCH 38.0
END DESCRIPTION:
XS GIS Cut Line= 4
      3815099.61     10506310.19      3814583.10     10505832.39
      3813805.32     10505749.06      3812555.29     10505547.67
#Sta/Elev= 30
  3906.3  389.98  4161.2  381.82  4515.0  375.11  4633.5  373.92  4673.1  375.09
  4754.2  373.35  4798.5  375.01  4854.8  373.22  4885.0  374.70  4945.3  372.38
  4985.5  372.99  4995.6  370.41  5025.8  372.66  5166.6  372.24  5241.4  370.60
  5333.3  371.43  5419.9  372.72  5496.2  370.36  5499.0  369.86  5502.2  370.36
  5505.0  370.51  5543.5  373.46  5590.4  371.78  5912.6  378.08  6166.8  383.74
  6350.1  391.10  6370.3  393.52  6390.6  393.25  6552.9  401.35  6658.3  402.29
#Mann=7,-1,0
  3906.3    0.05       0  4798.5    0.16       0  5333.3    0.05       0
  5496.2    0.07       0  5502.2    0.05       0  5505.0    0.16       0
  5912.6    0.05       0
Bank Sta=5496.2,5502.2
Exp/Cntr=0.3,0.1

Type RM Length L Ch R = 1,18023,442,442,442
BEGIN DESCRIPTION:
SIMS BRANCH 37.0
END DESCRIPTION:
XS GIS Cut Line= 4
      3815448.53     10505940.94      3814869.12     10505376.71
      3813731.96     10504738.69      3812903.76     10504706.17
#Sta/Elev= 30
  3308.8  389.91  3365.1  389.62  3513.7  384.58  3570.3  385.11  3598.6  383.07
  3768.1  379.01  4408.1  371.23  4429.8  367.54  4438.0  370.42  4487.0  371.83
  4656.8  370.38  4737.8  371.73  4827.9  370.07  4856.5  366.98  4878.2  369.11
  4980.9  370.02  4999.5  366.29  5002.3  365.79  5005.5  366.29  5018.5  366.72
  5024.2  368.86  5040.2  366.93  5045.9  370.40  5182.8  375.58  5332.4  384.22
  5391.6  385.68  5654.0  377.87  5767.3  377.28  5974.2  380.91  6250.3  391.75
#Mann=5,-1,0
  3308.8    0.05       0  4487.0    0.16       0  4999.5    0.07       0
  5005.5    0.16       0  5182.8    0.05       0
Bank Sta=4999.5,5005.5
Exp/Cntr=0.3,0.1

Type RM Length L Ch R = 1,17581,205,205,205
BEGIN DESCRIPTION:
SIMS BRANCH 36.0
END DESCRIPTION:
XS GIS Cut Line= 4
      3815534.52     10505137.96      3814596.99     10504818.50
      3814117.82     10504700.45      3812840.09     10504506.01
#Sta/Elev= 30
  3846.6  400.07  3904.6  399.80  4038.9  389.83  4195.7  384.06  4824.6  369.39
  4902.0  368.04  4927.1  365.59  4933.4  368.14  4974.9  368.55  5006.4  365.53
  5009.2  365.03  5012.4  365.53  5016.4  367.45  5026.6  368.08  5122.7  368.65
  5140.9  365.67  5146.0  368.21  5287.5  369.16  5428.9  374.05  5432.6  373.99
  5528.1  380.02  5581.6  384.08  5612.0  384.17  5697.9  388.81  5773.8  383.93
  5935.7  378.60  6163.2  379.15  6364.1  383.07  6621.7  393.69  6623.0  393.69
#Mann=10,-1,0
  3846.6    0.05       0  4824.6    0.16       0  4902.0    0.05       0
  5006.4    0.04       0  5012.4    0.05       0  5026.6    0.16       0
  5428.9    0.05       0  5432.6    0.08       0  5528.1    0.05       0
  6621.7    0.08       0
Bank Sta=5006.4,5012.4
Exp/Cntr=0.3,0.1

Type RM Length L Ch R = 1,17376,729,729,729
BEGIN DESCRIPTION:
SIMS BRANCH 35.0
END DESCRIPTION:
XS GIS Cut Line= 5
      3815472.00     10504915.73      3814416.44     10504631.00
      3814117.82     10504533.78      3813721.99     10504436.56
      3813006.69     10504339.34
#Sta/Elev= 30
  4070.1  395.30  4147.9  394.70  4414.3  389.53  4424.7  387.18  4498.5  387.93
  4600.8  380.47  4613.0  382.39  4672.6  378.55  4853.2  373.42  4932.2  368.94
  4951.6  371.45  4956.7  368.87  4984.0  368.40  5001.7  365.44  5004.5  364.94
  5007.7  365.44  5015.1  368.01  5060.1  368.48  5268.7  368.41  5378.3  369.00
  5671.3  375.57  5681.3  376.48  5761.9  380.14  5893.8  380.82  5907.6  379.07
  6171.0  375.44  6369.5  380.13  6468.7  384.28  6513.1  389.03  6606.9  391.00
#Mann=15,-1,0
  4070.1    0.05       0  4147.9    0.08       0  4414.3    0.05       0
  4672.6    0.08       0  4853.2    0.16       0  5001.7    0.07       0
  5007.7    0.16       0  5060.1    0.08       0  5268.7    0.16       0
  5378.3    0.05       0  5671.3    0.08       0  5681.3    0.05       0
  6171.0    0.08       0  6369.5    0.05       0  6468.7    0.08       0
Bank Sta=5001.7,5007.7
Exp/Cntr=0.3,0.1

Type RM Length L Ch R = 1,16647,432,432,432
BEGIN DESCRIPTION:
SIMS BRANCH 34.0
END DESCRIPTION:
XS GIS Cut Line= 3
      3815041.40     10504276.83      3814006.71     10504033.78
      3813667.81     10503764.04
#Sta/Elev= 30
  4261.3  391.87  4315.9  390.34  4378.6  386.71  4478.9  381.75  4519.9  378.58
  4632.9  373.68  4653.5  371.76  4660.3  370.03  4665.5  370.38  4684.3  368.24
  4776.7  365.60  4967.5  365.76  4982.2  365.44  4999.7  362.89  5002.5  362.39
  5005.7  362.89  5015.0  365.78  5101.0  364.92  5115.7  366.06  5126.0  365.21
  5177.4  365.87  5227.1  368.29  5259.5  367.57  5310.9  368.29  5374.0  370.50
  5402.9  372.54  5516.6  375.17  5659.1  385.95  5708.8  387.84  5757.3  387.69
#Mann=5,-1,0
  4261.3    0.05       0  4378.6    0.16       0  4999.7    0.07       0
  5005.7    0.16       0  5101.0    0.05       0
Bank Sta=4999.7,5005.7
Exp/Cntr=0.3,0.1

Type RM Length L Ch R = 1,16215,535,535,535
BEGIN DESCRIPTION:
SIMS BRANCH 33.0
END DESCRIPTION:
XS GIS Cut Line= 3
      3815013.64     10504144.88      3814617.82     10503797.67
      3813735.87     10503693.50
#Sta/Elev= 30
  4152.1  387.89  4236.6  387.48  4363.8  382.93  4370.4  383.32  4378.0  381.70
  4392.3  380.62  4413.1  380.26  4527.0  372.53  4547.9  372.61  4583.1  370.33
  4640.0  368.73  4827.9  365.78  4888.3  362.94  4954.6  364.60  4978.9  364.34
  4999.0  363.24  5006.1  359.98  5008.9  359.48  5012.1  359.98  5019.2  363.70
  5044.9  364.39  5240.7  375.35  5250.8  376.76  5281.0  377.32  5301.4  379.28
  5401.8  383.49  5411.9  384.71  5452.2  386.17  5492.5  388.85  5566.7  389.78
#Mann=5,-1,0
  4152.1    0.05       0  4640.0    0.16       0  5006.1    0.07       0
  5012.1    0.16       0  5044.9    0.05       0
Bank Sta=5006.1,5012.1
Exp/Cntr=0.3,0.1

Type RM Length L Ch R = 1,15680,440,440,440
BEGIN DESCRIPTION:
SIMS BRANCH 32.0
END DESCRIPTION:
XS GIS Cut Line= 3
      3815472.00     10503165.73      3814499.77     10503360.17
      3813792.99     10503374.03
#Sta/Elev= 30
  3876.1  382.86  3919.3  382.33  3929.5  381.49  3970.3  380.95  4031.5  378.57
  4204.9  374.10  4439.4  370.02  4521.0  370.59  4633.4  369.00  4776.0  363.86
  4827.0  362.91  4842.2  361.18  4857.5  362.55  4967.8  363.05  4987.8  359.17
  4994.8  358.62  4997.5  358.12  5000.8  358.62  5007.8  359.35  5017.8  362.19
  5037.8  363.38  5067.8  363.78  5098.5  365.68  5117.8  365.98  5237.8  374.17
  5317.8  378.54  5357.8  381.89  5457.9  387.44  5497.9  388.40  5574.5  386.97
#Mann=5,-1,0
  3876.1    0.05       0  4633.4    0.16       0  4994.8    0.07       0
  5000.8    0.16       0  5098.5    0.05       0
Bank Sta=4994.8,5000.8
Exp/Cntr=0.3,0.1

Type RM Length L Ch R = 1,15240,711,711,711
BEGIN DESCRIPTION:
SIMS BRANCH 31.0
END DESCRIPTION:
XS GIS Cut Line= 3
      3815201.18     10502839.33      3814319.21     10503026.84
      3813826.15     10503269.90
#Sta/Elev= 30
  4295.8  382.73  4310.6  382.67  4338.3  382.89  4522.3  379.40  4561.3  379.92
  4679.7  378.76  4747.2  376.66  4875.6  369.85  4972.2  363.40  4982.4  362.12
  4992.3  356.66  4999.8  354.72  5002.6  354.22  5005.8  354.72  5013.1  358.46
  5033.5  362.18  5146.3  362.32  5166.4  361.42  5265.6  362.27  5304.9  365.02
  5310.5  364.42  5327.3  366.79  5332.9  366.48  5377.8  370.61  5394.7  373.01
  5448.8  377.30  5535.0  381.69  5609.6  383.42  5631.8  384.92  5747.2  384.47
#Mann=7,-1,0
  4295.8    0.05       0  4310.6    0.16       0  4679.7    0.05       0
  4875.6    0.16       0  4999.8    0.07       0  5005.8    0.16       0
  5448.8    0.05       0
Bank Sta=4999.8,5005.8
Exp/Cntr=0.3,0.1

Type RM Length L Ch R = 1,14529,254,254,254
BEGIN DESCRIPTION:
SIMS BRANCH 30.0
END DESCRIPTION:
XS GIS Cut Line= 4
      3815055.36     10502728.24      3814603.94     10502575.45
      3814048.38     10502721.28      3813756.71     10503193.51
#Sta/Elev= 30
  4112.1  380.96  4279.7  378.63  4374.0  378.82  4562.6  373.95  4717.2  367.50
  4749.3  367.61  4779.3  364.29  4860.1  359.86  4872.3  361.11  4955.0  361.01
  4975.7  356.83  4978.2  353.86  4980.9  353.36  4984.2  353.86  4996.4  354.22
  5006.7  358.22  5027.4  360.54  5048.1  358.44  5068.7  360.60  5079.1  358.10
  5110.1  360.17  5151.5  357.64  5159.8  361.48  5165.4  361.48  5174.8  365.37
  5196.8  368.82  5232.8  372.50  5314.6  376.43  5531.9  376.36  5718.1  380.70
#Mann=4,-1,0
  4112.1    0.16       0  4978.2    0.07       0  4984.2    0.16       0
  5196.8    0.05       0
Bank Sta=4978.2,4984.2
Exp/Cntr=0.3,0.1

Type RM Length L Ch R = 1,14275,492,492,492
BEGIN DESCRIPTION:
SIMS BRANCH 29.0
END DESCRIPTION:
XS GIS Cut Line= 4
      3815374.74     10502603.22      3814569.21     10502360.17
      3814041.44     10502457.39      3813097.01     10502561.56
#Sta/Elev= 30
  3744.0  381.40  4231.4  374.02  4294.4  373.88  4334.3  378.51  4344.7  376.02
  4365.6  374.21  4447.6  374.69  4679.4  371.97  4775.9  366.92  4849.4  359.96
  4892.1  358.68  4981.6  359.51  4991.7  358.53  5000.2  353.36  5003.0  352.86
  5006.2  353.36  5032.4  358.69  5103.6  357.73  5114.3  359.03  5120.4  356.10
  5125.5  356.10  5133.9  360.29  5202.5  360.67  5366.2  359.27  5378.0  357.93
  5468.9  362.90  5476.0  365.32  5520.2  365.59  5818.1  375.16  6072.2  378.47
#Mann=9,-1,0
  3744.0    0.05       0  4231.4    0.16       0  4447.6    0.05       0
  4679.4    0.16       0  5000.2    0.07       0  5006.2    0.16       0
  5202.5    0.05       0  5366.2    0.16       0  5520.2    0.05       0
Bank Sta=5000.2,5006.2
Exp/Cntr=0.3,0.1

Type RM Length L Ch R = 1,13783,459,459,459
BEGIN DESCRIPTION:
SIMS BRANCH 28.0
END DESCRIPTION:
XS GIS Cut Line= 3
      3814149.58     10501860.21      3813898.79     10502080.95
      3813244.04     10502202.36
#Sta/Elev= 30
  4698.8  370.49  4850.7  361.15  4861.5  361.24  4932.6  357.52  4975.3  358.24
  4986.5  352.26  4989.3  351.76  4992.5  352.26  4996.2  354.36  5003.8  354.97
  5010.4  358.19  5018.0  357.31  5042.2  357.16  5103.3  358.17  5114.8  357.07
  5154.1  357.31  5194.8  355.76  5205.0  357.94  5215.1  358.19  5220.5  359.83
  5235.5  360.85  5245.6  363.27  5286.2  364.18  5377.9  367.26  5449.0  372.02
  5479.6  373.26  5500.0  375.62  5530.4  375.26  5605.7  377.36  5698.8  375.36
#Mann=5,-1,0
  4698.8    0.05       0  4850.7    0.16       0  4986.5    0.07       0
  4992.5    0.16       0  5286.2    0.05       0
Bank Sta=4986.5,4992.5
Exp/Cntr=0.3,0.1

Type RM Length L Ch R = 1,13324,439,439,439
BEGIN DESCRIPTION:
SIMS BRANCH 27.0
END DESCRIPTION:
XS GIS Cut Line= 4
      3814049.59     10501660.19      3813649.61     10501710.19
      3813499.61     10501810.19      3813260.77     10502020.18
#Sta/Elev= 30
  4598.7  367.18  4659.1  364.08  4672.2  362.93  4709.5  360.56  4717.1  359.31
  4759.9  356.41  4797.7  355.33  4890.9  356.02  4901.0  355.54  4981.6  356.93
  4991.7  356.66  4996.3  350.52  4999.0  350.02  5002.3  350.52  5004.8  350.52
  5009.3  355.82  5015.3  352.31  5024.3  357.85  5030.3  357.16  5045.4  359.79
  5075.1  361.45  5102.5  362.10  5132.5  364.09  5146.0  364.19  5153.5  365.29
  5174.6  366.57  5179.1  367.66  5260.3  372.57  5387.5  374.35  5500.1  373.05
#Mann=5,-1,0
  4598.7    0.05       0  4672.2    0.16       0  4996.3    0.07       0
  5002.3    0.16       0  5075.1    0.05       0
Bank Sta=4996.3,5002.3
Exp/Cntr=0.3,0.1

Type RM Length L Ch R = 1,12885,90,90,90
BEGIN DESCRIPTION:
Mapping XS 0e866212
END DESCRIPTION:
XS GIS Cut Line= 3
      3814627.91     10501720.69      3813560.24     10501386.50
      3813123.27     10501325.93
#Sta/Elev= 30
  4177.0  374.16  4225.6  374.88  4258.1  373.51  4280.0  374.74  4290.5  373.25
  4360.7  372.53  4384.8  373.36  4398.4  372.34  4625.6  372.37  4678.2  371.40
  4756.8  367.02  4798.3  365.61  4830.8  361.75  4893.3  357.79  4933.4  355.32
  4982.1  355.70  4992.5  349.87  4995.3  349.85  4998.1  349.35  5001.3  349.85
  5024.0  354.96  5044.9  353.49  5100.9  356.07  5133.4  356.21  5139.2  355.22
  5302.6  358.32  5401.9  362.01  5528.7  366.31  5690.1  373.71  5736.9  374.16
#Mann=7,-1,0
  4177.0    0.05       0  4756.8    0.08       0  4893.3    0.05       0
  4995.3    0.04       0  5001.3    0.05       0  5302.6    0.08       0
  5401.9    0.05       0
Bank Sta=4995.3,5001.3
Exp/Cntr=0.3,0.1

Type RM Length L Ch R = 1,12795,553,553,553
BEGIN DESCRIPTION:
SIMS BRANCH 26.0
END DESCRIPTION:
XS GIS Cut Line= 2
      3814688.69     10501633.89      3813195.71     10501195.54
#Sta/Elev= 30
  4164.2  376.09  4319.6  373.31  4369.5  373.85  4408.1  372.29  4618.8  370.72
  4624.0  369.91  4684.3  369.65  4732.6  367.15  4762.8  364.75  4768.0  363.12
  4778.1  363.10  4809.4  359.44  4821.4  359.11  4882.4  354.72  4973.5  354.87
  4986.6  353.45  4997.0  350.24  5003.9  350.09  5006.6  349.59  5009.9  350.09
  5012.1  353.19  5017.9  355.16  5090.8  354.10  5174.2  354.79  5222.8  356.42
  5288.8  356.28  5466.0  362.44  5486.8  364.45  5518.1  364.62  5720.2  371.71
#Mann=5,-1,0
  4164.2    0.05       0  4732.6    0.08       0  4821.4    0.05       0
  5003.9    0.04       0  5009.9    0.05       0
Bank Sta=5003.9,5009.9
Exp/Cntr=0.3,0.1

Type RM Length L Ch R = 1,12242,558,558,558
BEGIN DESCRIPTION:
SIMS BRANCH 25.0
END DESCRIPTION:
XS GIS Cut Line= 3
      3814549.61     10501010.19      3813949.61     10500960.19
      3813249.60     10501160.19
#Sta/Elev= 30
  4385.9  373.55  4448.6  371.49  4516.4  367.95  4684.4  357.88  4697.0  358.31
  4757.2  354.99  4837.5  352.24  4889.5  352.13  4921.9  351.80  4957.9  350.70
  4977.9  351.64  4985.5  349.52  4990.6  349.52  4995.4  347.17  4998.1  346.67
  5001.4  347.17  5004.9  351.58  5010.1  350.22  5019.2  351.79  5071.2  350.91
  5189.5  353.99  5248.0  353.22  5289.6  353.71  5424.8  358.59  5475.5  361.96
  5587.3  365.80  5592.5  365.37  5660.1  368.85  5684.8  368.63  5716.0  370.31
#Mann=5,-1,0
  4385.9    0.05       0  4889.5    0.16       0  4921.9    0.05       0
  4995.4    0.03       0  5001.4    0.05       0
Bank Sta=4995.4,5001.4
Exp/Cntr=0.3,0.1

Type RM Length L Ch R = 1,11684,474,474,474
BEGIN DESCRIPTION:
SIMS BRANCH 24.0
END DESCRIPTION:
XS GIS Cut Line= 4
      3814423.94     10500527.12      3813950.87     10500449.00
      3813390.97     10500705.08      3813165.27     10501052.31
#Sta/Elev= 30
  4105.3  365.15  4238.2  361.23  4383.3  358.06  4515.1  362.61  4548.7  362.95
  4575.9  361.76  4595.7  362.49  4618.7  362.06  4641.1  360.95  4652.7  359.11
  4685.1  357.08  4698.7  355.37  4762.1  351.25  4850.1  350.03  4872.1  349.05
  4888.4  349.67  4911.4  346.67  4939.9  348.70  4962.9  349.18  4980.4  348.26
  5000.5  344.49  5003.2  343.99  5006.5  344.49  5009.0  344.87  5015.0  348.46
  5026.0  350.04  5147.0  353.24  5313.9  362.19  5487.1  367.14  5614.6  368.47
#Mann=3,-1,0
  4105.3    0.05       0  5000.5    0.03       0  5006.5    0.05       0
Bank Sta=5000.5,5006.5
Exp/Cntr=0.3,0.1

Type RM Length L Ch R = 1,11210,418,418,418
BEGIN DESCRIPTION:
SIMS BRANCH 23.0
END DESCRIPTION:
XS GIS Cut Line= 3
      3813929.49     10500409.27      3813371.72     10500250.84
      3813230.66     10500834.61
#Sta/Elev= 30
  4534.2  362.12  4627.6  357.31  4729.3  353.24  4734.5  353.72  4742.0  352.43
  4807.4  349.68  4841.3  347.18  4897.9  347.23  4948.2  345.96  4970.7  346.77
  4981.1  346.56  4987.3  344.41  4998.9  344.26  5001.6  343.76  5004.9  344.26
  5033.1  348.75  5112.5  352.17  5141.7  351.67  5146.8  352.39  5183.6  350.74
  5225.4  350.62  5247.1  351.60  5257.4  351.30  5278.0  352.59  5308.8  352.66
  5319.4  353.48  5452.9  356.83  5570.6  358.27  5696.2  362.38  5714.6  362.38
#Mann=3,-1,0
  4534.2    0.05       0  4998.9    0.03       0  5004.9    0.05       0
Bank Sta=4998.9,5004.9
Exp/Cntr=0.3,0.1

Type RM Length L Ch R = 1,10792,527,527,527
BEGIN DESCRIPTION:
SIMS BRANCH 22.0
END DESCRIPTION:
XS GIS Cut Line= 3
      3813899.58     10500360.16      3813599.61     10499960.19
      3813048.07     10499793.62
#Sta/Elev= 30
  4506.7  359.15  4614.0  354.31  4693.1  352.10  4734.8  350.31  4864.0  348.67
  4934.8  346.39  4964.0  346.14  4970.2  344.17  4978.5  344.02  4984.8  340.05
  4996.4  339.50  4999.1  339.00  5002.4  339.50  5009.3  339.83  5017.1  342.61
  5038.0  344.10  5100.7  346.00  5198.4  347.03  5205.1  346.05  5215.6  345.83
  5236.6  343.97  5246.9  346.04  5278.3  348.33  5302.5  348.96  5335.5  350.86
  5340.9  352.11  5373.7  355.51  5406.6  356.28  5487.2  359.81  5582.8  361.03
#Mann=3,-1,0
  4506.7    0.05       0  4996.4    0.03       0  5002.4    0.05       0
Bank Sta=4996.4,5002.4
Exp/Cntr=0.3,0.1

Type RM Length L Ch R = 1,10265,397,397,397
BEGIN DESCRIPTION:
SIMS BRANCH 21.0
END DESCRIPTION:
XS GIS Cut Line= 2
      3814419.66     10499958.57      3813270.01     10499294.82
#Sta/Elev= 30
  4154.4  366.58  4203.8  365.68  4262.7  363.42  4278.4  362.04  4315.8  360.33
  4498.1  353.02  4578.5  350.76  4686.3  348.87  4717.8  345.93  4766.7  343.58
  4862.9  342.45  4900.2  342.93  4937.5  342.27  4943.3  341.41  4980.6  342.63
  4986.4  341.66  4991.0  339.34  4996.4  336.61  4999.2  336.58  5001.9  336.08
  5005.2  336.58  5008.9  339.29  5017.9  340.54  5093.4  342.97  5119.9  344.33
  5170.6  349.05  5251.4  353.17  5339.6  354.89  5435.8  359.08  5481.9  359.68
#Mann=5,-1,0
  4154.4    0.05       0  4991.0    0.16       0  4999.2    0.07       0
  5005.2    0.16       0  5093.4    0.05       0
Bank Sta=4999.2,5005.2
Exp/Cntr=0.3,0.1

Type RM Length L Ch R = 1,9868,472,472,472
BEGIN DESCRIPTION:
SIMS BRANCH 20.0
END DESCRIPTION:
XS GIS Cut Line= 3
      3814389.24     10499758.90      3813999.61     10499460.19
      3813599.58     10499110.16
#Sta/Elev= 30
  4533.6  363.50  4583.1  361.26  4603.9  359.74  4624.8  359.47  4653.8  357.38
  4732.7  353.98  4903.1  348.77  4961.1  348.02  4982.0  340.37  4985.3  333.84
  4988.0  333.34  4991.3  333.84  5002.8  333.94  5011.0  336.83  5014.0  336.63
  5027.9  336.48  5031.7  338.05  5045.9  339.76  5088.6  341.95  5102.9  341.28
  5138.0  342.26  5194.9  342.17  5223.4  340.87  5280.2  342.71  5350.6  344.63
  5399.9  345.28  5442.6  347.07  5463.5  348.96  5485.4  350.04  5556.1  352.48
#Mann=5,-1,0
  4533.6    0.05       0  4985.3    0.03       0  4991.3    0.05       0
  5014.0    0.16       0  5280.2    0.05       0
Bank Sta=4985.3,4991.3
Exp/Cntr=0.3,0.1

Type RM Length L Ch R = 1,9396,404,404,404
BEGIN DESCRIPTION:
SIMS BRANCH 19.0
END DESCRIPTION:
XS GIS Cut Line= 3
      3814632.31     10499737.23      3814298.09     10499133.90
      3813749.61     10498810.19
#Sta/Elev= 30
  4082.6  364.67  4216.4  363.97  4273.6  361.08  4281.7  359.91  4303.5  358.72
  4347.0  358.41  4434.0  355.17  4569.1  353.21  4672.1  349.16  4693.9  347.93
  4721.4  345.04  4743.1  344.74  4794.5  341.50  4823.9  340.62  4933.1  338.65
  4948.7  337.54  4970.1  337.69  4979.6  336.60  4991.6  333.57  4998.4  333.22
  5001.2  332.72  5004.4  333.22  5007.2  333.86  5014.4  337.41  5022.9  338.41
  5040.4  338.44  5087.2  340.44  5161.4  341.87  5262.8  348.13  5409.2  351.53
#Mann=5,-1,0
  4082.6    0.05       0  4823.9    0.16       0  4998.4    0.07       0
  5004.4    0.16       0  5040.4    0.05       0
Bank Sta=4998.4,5004.4
Exp/Cntr=0.3,0.1

Type RM Length L Ch R = 1,8992,717,717,717
BEGIN DESCRIPTION:
SIMS BRANCH 18.0
END DESCRIPTION:
XS GIS Cut Line= 3
      3815092.35     10498838.76      3814002.95     10498613.06
      3813353.21     10498600.07
#Sta/Elev= 30
  4088.3  354.01  4244.3  351.88  4357.0  349.11  4497.4  342.40  4502.5  343.71
  4602.8  341.40  4647.9  339.38  4748.3  339.02  4806.0  336.39  4848.6  336.03
  4877.5  334.58  4892.9  335.99  4928.5  337.18  4979.6  335.50  4988.9  330.44
  4997.0  328.99  4999.8  328.49  5003.0  328.99  5010.2  334.63  5020.4  337.47
  5030.6  339.45  5054.6  340.34  5291.9  346.87  5302.8  347.19  5404.2  350.08
  5424.2  348.53  5434.2  348.81  5455.1  351.33  5811.6  358.99  5850.7  359.97
#Mann=9,-1,0
  4088.3    0.05       0  4892.9    0.16       0  4997.0    0.07       0
  5003.0    0.16       0  5054.6    0.05       0  5291.9    0.16       0
  5302.8    0.05       0  5455.1    0.16       0  5811.6    0.05       0
Bank Sta=4997,5003
Exp/Cntr=0.3,0.1

Type RM Length L Ch R = 1,8275,384,384,384
BEGIN DESCRIPTION:
SIMS BRANCH 17.0
END DESCRIPTION:
XS GIS Cut Line= 2
      3814955.18     10498471.56      3813670.44     10498006.28
#Sta/Elev= 30
  4263.8  349.22  4599.4  339.98  4661.1  337.27  4697.1  337.97  4727.7  336.54
  4753.0  336.85  4768.8  335.38  4870.2  336.15  4876.0  337.37  4886.6  335.73
  4926.2  334.37  4931.5  332.62  4939.8  331.98  4962.2  333.74  4987.5  332.07
  4992.9  329.04  5003.6  326.21  5015.1  325.89  5017.9  325.39  5021.1  325.89
  5024.9  333.39  5135.3  335.72  5141.8  337.01  5191.3  339.94  5196.6  339.32
  5285.4  343.52  5339.2  346.01  5369.8  345.99  5425.8  349.17  5630.2  355.02
#Mann=5,-1,0
  4263.8    0.05       0  4768.8    0.16       0  5015.1    0.07       0
  5021.1    0.16       0  5285.4    0.05       0
Bank Sta=5015.1,5021.1
Exp/Cntr=0.3,0.1

Type RM Length L Ch R = 1,7891,623,623,623
BEGIN DESCRIPTION:
SIMS BRANCH 16.0
END DESCRIPTION:
XS GIS Cut Line= 3
      3814949.59     10498310.18      3814316.32     10497936.85
      3813799.63     10497910.19
#Sta/Elev= 30
  4355.9  348.57  4363.7  348.84  4369.5  347.16  4379.1  346.77  4560.8  340.82
  4603.7  341.42  4634.5  340.56  4640.8  339.10  4720.9  337.28  4773.6  339.37
  4933.6  334.76  4947.9  333.69  4955.1  331.55  4970.7  330.63  4982.7  331.26
  4992.2  328.99  4998.0  323.66  5002.9  323.62  5005.7  323.12  5008.9  323.62
  5013.6  324.53  5019.4  327.68  5035.1  331.51  5107.8  331.56  5123.0  327.28
  5147.8  331.65  5187.9  333.08  5197.5  334.43  5398.1  342.34  5608.4  352.95
#Mann=4,-1,0
  4355.9    0.16       0  5002.9    0.07       0  5008.9    0.16       0
  5197.5    0.05       0
Bank Sta=5002.9,5008.9
Exp/Cntr=0.3,0.1

Type RM Length L Ch R = 1,7268,429,429,429
BEGIN DESCRIPTION:
SIMS BRANCH 15.0
END DESCRIPTION:
XS GIS Cut Line= 3
      3815099.57     10498110.16      3814449.61     10497660.19
      3814099.63     10497560.20
#Sta/Elev= 30
  4208.7  349.33  4237.0  345.91  4302.6  345.22  4359.3  341.83  4568.1  336.52
  4589.1  337.57  4683.0  335.51  4768.1  331.71  4812.7  332.78  4877.6  330.19
  4884.4  327.09  4890.4  330.44  4914.1  327.88  4976.9  329.61  4985.7  327.48
  4996.2  321.20  5006.6  319.09  5009.4  318.59  5012.6  319.09  5030.4  327.80
  5049.9  329.53  5055.1  326.52  5082.4  330.90  5088.9  329.34  5103.2  331.05
  5122.7  330.32  5127.9  332.81  5161.7  335.64  5307.6  343.98  5363.2  346.78
#Mann=4,-1,0
  4208.7    0.16       0  5006.6    0.07       0  5012.6    0.16       0
  5307.6    0.05       0
Bank Sta=5006.6,5012.6
Exp/Cntr=0.3,0.1

Type RM Length L Ch R = 1,6839,463,463,463
BEGIN DESCRIPTION:
SIMS BRANCH 14.0
END DESCRIPTION:
XS GIS Cut Line= 3
      3815121.89     10497777.14      3814699.61     10497460.19
      3814299.61     10497210.19
#Sta/Elev= 30
  4491.1  342.78  4597.3  338.86  4805.6  335.96  4811.8  335.13  4819.0  336.28
  4869.1  334.12  4891.0  334.27  4955.6  330.82  4961.8  329.22  4969.1  331.75
  4976.4  331.42  4988.0  319.30  4990.7  318.80  4994.0  319.30  4997.2  319.35
  5005.6  322.30  5011.8  326.16  5026.8  326.22  5032.7  327.34  5063.3  325.93
  5162.9  327.06  5184.8  326.74  5266.7  329.47  5302.1  333.00  5331.0  333.54
  5352.2  336.28  5419.5  341.96  5446.6  342.93  5467.8  345.80  5490.8  347.09
#Mann=4,-1,0
  4491.1    0.16       0  4988.0    0.07       0  4994.0    0.16       0
  5162.9    0.05       0
Bank Sta=4988,4994
Exp/Cntr=0.3,0.1

Type RM Length L Ch R = 1,6376,556,556,556
BEGIN DESCRIPTION:
SIMS BRANCH 13.0
END DESCRIPTION:
XS GIS Cut Line= 3
      3815049.58     10497260.15      3814949.61     10497110.19
      3814549.64     10496960.20
#Sta/Elev= 30
  4811.9  331.68  4825.4  331.09  4861.4  327.68  4884.0  326.06  4906.5  325.56
  4948.6  327.95  4956.1  327.09  4963.6  323.46  4969.6  318.72  4986.1  317.11
  4988.9  316.61  4992.1  317.11  5007.3  317.81  5013.5  319.70  5024.2  320.04
  5032.2  321.83  5041.5  322.18  5067.8  325.77  5087.4  326.86  5141.6  326.80
  5147.9  327.35  5178.1  327.78  5259.0  330.78  5283.0  331.92  5312.5  333.16
  5349.0  336.91  5365.9  337.28  5387.3  338.52  5404.2  340.28  5419.3  341.25
#Mann=6,-1,0
  4811.9    0.16       0  4986.1    0.07       0  4992.1    0.16       0
  5041.5    0.05       0  5259.0     0.1       0  5283.0    0.05       0
Bank Sta=4986.1,4992.1
Exp/Cntr=0.3,0.1

Type RM Length L Ch R = 1,5820,417,417,417
BEGIN DESCRIPTION:
SIMS BRANCH 12.0
END DESCRIPTION:
XS GIS Cut Line= 3
      3815199.61     10497260.20      3815199.61     10496860.19
      3814899.59     10496560.17
#Sta/Elev= 30
  4585.3  335.63  4670.4  329.62  4744.0  325.47  4775.3  324.91  4866.7  324.97
  4885.3  324.38  4915.3  321.53  4925.3  322.76  4935.3  323.05  4975.3  321.50
  4982.8  318.87  4988.8  318.87  4996.5  314.56  4999.2  314.06  5002.5  314.56
  5013.6  319.70  5027.7  320.50  5041.9  322.14  5056.0  322.73  5070.2  321.79
  5084.3  322.87  5098.4  326.15  5112.6  328.16  5140.9  327.87  5155.0  328.36
  5211.6  330.86  5225.7  331.99  5310.6  334.46  5338.9  336.18  5409.6  338.91
#Mann=6,-1,0
  4585.3    0.16       0  4670.4    0.05       0  4744.0    0.16       0
  4866.7    0.05       0  4996.5    0.03       0  5002.5    0.05       0
Bank Sta=4996.5,5002.5
Exp/Cntr=0.3,0.1

Type RM Length L Ch R = 1,5403,342,342,342
BEGIN DESCRIPTION:
SIMS BRANCH 11.0
END DESCRIPTION:
XS GIS Cut Line= 3
      3815899.61     10496910.19      3815499.61     10496660.19
      3815149.59     10496360.17
#Sta/Elev= 30
  4509.0  334.30  4616.9  330.55  4684.1  326.75  4851.0  322.88  4915.3  319.76
  4945.3  321.82  4967.1  320.85  4973.0  321.90  4977.8  319.59  4984.0  319.59
  4987.8  314.96  4991.4  312.17  4994.2  311.67  4997.4  312.17  5002.1  312.19
  5016.4  317.57  5030.6  319.22  5044.9  319.57  5051.5  318.40  5080.0  319.94
  5108.6  324.98  5129.4  325.61  5137.1  326.90  5158.0  326.59  5172.2  327.93
  5200.8  328.15  5229.3  328.08  5235.9  326.91  5285.3  329.89  5441.7  334.56
#Mann=3,-1,0
  4509.0    0.05       0  4991.4    0.03       0  4997.4    0.05       0
Bank Sta=4991.4,4997.4
Exp/Cntr=0.3,0.1

Type RM Length L Ch R = 1,5061,458,458,458
BEGIN DESCRIPTION:
SIMS BRANCH 10.0
END DESCRIPTION:
XS GIS Cut Line= 2
      3816217.38     10496679.92      3815300.73     10496238.95
#Sta/Elev= 30
  4375.7  342.62  4495.3  339.53  4561.9  336.30  4591.9  333.83  4642.7  332.54
  4739.4  326.80  4817.1  323.25  4914.3  319.64  4965.1  318.72  4982.2  316.23
  4987.7  312.85  4991.7  311.31  4994.4  310.81  4997.7  311.31  5004.8  311.82
  5016.9  314.80  5027.5  315.79  5033.0  314.75  5050.1  314.31  5055.6  313.26
  5083.8  314.72  5100.9  317.34  5106.4  316.86  5129.1  318.54  5146.2  321.28
  5168.8  322.10  5174.3  323.19  5219.6  326.36  5272.1  328.92  5392.9  332.81
#Mann=3,-1,0
  4375.7    0.05       0  4991.7    0.03       0  4997.7    0.05       0
Bank Sta=4991.7,4997.7
Exp/Cntr=0.3,0.1

Type RM Length L Ch R = 1,4603,604,604,604
BEGIN DESCRIPTION:
SIMS BRANCH 9.0
END DESCRIPTION:
XS GIS Cut Line= 3
      3816203.48     10496468.11      3815946.53     10496079.21
      3815189.62     10495891.72
#Sta/Elev= 30
  4381.3  339.94  4439.2  337.45  4570.6  334.79  4722.2  327.01  4728.2  326.09
  4830.5  321.81  4875.2  319.23  4937.0  317.68  4978.2  318.80  4986.1  318.35
  4995.8  309.52  4998.5  309.02  5001.8  309.52  5019.4  315.59  5091.5  316.23
  5110.3  318.87  5115.5  318.30  5122.4  321.34  5143.0  324.14  5184.2  327.30
  5193.1  327.67  5234.5  326.27  5281.1  326.75  5363.9  329.19  5462.4  333.15
  5565.4  335.62  5570.9  336.64  5586.0  336.93  5612.3  339.27  5627.2  339.16
#Mann=3,-1,0
  4381.3    0.05       0  4995.8    0.03       0  5001.8    0.05       0
Bank Sta=4995.8,5001.8
Exp/Cntr=0.3,0.1

Type RM Length L Ch R = 1,3999,75,75,75
BEGIN DESCRIPTION:
SIMS BRANCH 8.0
END DESCRIPTION:
XS GIS Cut Line= 3
      3816260.78     10496416.06      3815927.43     10495499.35
      3815323.96     10495218.42
#Sta/Elev= 30
  4259.0  340.07  4560.9  333.40  4644.0  330.47  4716.7  328.16  4742.0  328.69
  4772.7  326.95  4878.5  319.48  4945.5  312.39  4967.5  311.02  4984.4  311.93
  4996.5  308.50  4999.2  308.00  5002.5  308.50  5012.0  309.32  5020.7  312.47
  5042.6  314.53  5067.9  315.90  5090.3  314.85  5184.9  317.02  5210.2  316.02
  5309.3  320.16  5412.1  327.36  5480.7  327.45  5540.9  329.96  5737.9  333.02
  5760.8  333.86  5766.3  335.56  5794.7  335.35  5834.9  338.65  5900.1  340.45
#Mann=9,-1,0
  4259.0    0.05       0  4560.9    0.08       0  4644.0    0.05       0
  4772.7    0.08       0  4878.5    0.05       0  4984.4    0.08       0
  4996.5    0.07       0  5002.5    0.08       0  5090.3    0.05       0
Bank Sta=4996.5,5002.5
Exp/Cntr=0.3,0.1

Type RM Length L Ch R = 1,3924,346,346,346
BEGIN DESCRIPTION:
SIMS BRANCH 7.0
END DESCRIPTION:
XS GIS Cut Line= 5
      3816399.65     10496388.24      3816177.43     10495964.63
      3816031.60     10495575.74      3815973.44     10495396.92
      3815409.20     10495090.93
#Sta/Elev= 30
  4251.7  341.09  4621.6  331.12  4649.0  331.65  4688.7  331.03  4701.2  332.91
  4764.0  325.35  4769.4  326.75  4799.6  325.65  4845.9  321.70  4866.5  320.09
  4910.0  317.77  4934.9  312.67  4940.3  315.08  4948.4  310.50  4987.1  306.84
  4989.8  306.34  4993.1  306.84  4995.4  311.37  5001.8  308.55  5012.5  308.85
  5025.7  314.91  5184.7  315.16  5289.2  316.52  5371.9  318.91  5553.9  330.34
  5613.1  332.10  5754.8  331.93  5903.1  336.40  5904.0  336.48  5975.3  338.45
#Mann=11,-1,0
  4251.7    0.05       0  4621.6    0.08       0  4649.0    0.05       0
  4845.9    0.08       0  4866.5    0.05       0  4987.1    0.04       0
  4993.1    0.05       0  5184.7    0.08       0  5289.2    0.05       0
  5903.1    0.08       0  5904.0    0.05       0
Bank Sta=4987.1,4993.1
Exp/Cntr=0.3,0.1

Type RM Length L Ch R = 1,3578,551,551,551
BEGIN DESCRIPTION:
Mapping XS cb5fd9b5
END DESCRIPTION:
XS GIS Cut Line= 3
      3816861.45     10495844.83      3816147.92     10495360.46
      3815460.42     10494922.96
#Sta/Elev= 30
  4260.1  348.36  4401.6  344.81  4452.4  344.81  4479.9  344.36  4494.5  342.62
  4509.4  343.44  4553.6  339.54  4761.0  329.53  4769.9  327.88  4847.8  323.56
  4927.1  316.63  4934.6  314.84  4976.6  310.39  4985.1  306.86  4988.5  303.94
  4991.3  303.44  4994.5  303.94  5006.4  306.32  5012.5  310.53  5021.4  311.99
  5137.5  313.00  5296.2  318.57  5338.5  320.96  5374.9  324.98  5417.2  325.62
  5541.7  331.67  5593.3  333.33  5642.0  332.48  5736.9  333.68  5937.4  338.94
#Mann=7,-1,0
  4260.1    0.05       0  4452.4    0.08       0  4553.6    0.05       0
  4985.1    0.16       0  4988.5    0.07       0  4994.5    0.16       0
  5137.5    0.05       0
Bank Sta=4988.5,4994.5
Exp/Cntr=0.3,0.1

Type RM Length L Ch R = 1,3027,446,446,446
BEGIN DESCRIPTION:
SIMS BRANCH 6.0
END DESCRIPTION:
XS GIS Cut Line= 3
      3816799.64     10495310.21      3816399.61     10494960.19
      3815833.28     10494801.81
#Sta/Elev= 30
  4483.7  335.84  4576.3  326.80  4689.2  319.21  4717.7  318.23  4752.8  315.32
  4866.7  312.15  4895.2  310.53  4901.8  310.95  4916.1  309.01  4958.8  310.11
  4973.0  309.43  4979.7  304.94  4990.9  302.65  4993.6  302.15  4996.9  302.65
  5001.5  303.00  5008.1  308.96  5011.9  310.33  5071.6  310.07  5139.8  314.27
  5179.3  317.82  5202.1  321.65  5212.5  322.09  5223.8  324.16  5264.5  326.84
  5365.5  329.10  5444.2  329.41  5478.3  331.14  5534.4  329.69  5603.3  330.94
#Mann=3,-1,0
  4483.7    0.05       0  4990.9    0.03       0  4996.9    0.05       0
Bank Sta=4990.9,4996.9
Exp/Cntr=0.3,0.1

Type RM Length L Ch R = 1,2581,646,646,646
BEGIN DESCRIPTION:
SIMS BRANCH 5.0
END DESCRIPTION:
XS GIS Cut Line= 4
      3817121.88     10495219.84      3816856.25     10494756.29
      3816444.79     10494480.25      3815893.65     10494350.27
#Sta/Elev= 30
  4253.7  343.96  4299.4  343.30  4365.8  340.53  4495.3  332.56  4505.4  332.74
  4511.2  331.53  4629.1  326.65  4774.4  315.94  4883.0  309.56  4904.3  308.84
  4949.0  309.43  4976.6  308.22  4991.0  302.34  4997.0  301.16  4999.7  300.66
  5003.0  301.16  5012.7  302.56  5021.0  307.53  5091.9  308.02  5157.2  308.50
  5216.1  311.01  5283.4  316.54  5310.0  321.70  5371.0  326.40  5453.2  327.64
  5526.8  325.93  5627.8  326.47  5653.8  328.69  5701.2  328.22  5849.7  331.77
#Mann=4,-1,0
  4253.7    0.05       0  4997.0    0.03       0  5003.0    0.05       0
  5091.9    0.05       0
Bank Sta=4997,5003
Exp/Cntr=0.3,0.1

Type RM Length L Ch R = 1,1935,591,591,591
BEGIN DESCRIPTION:
SIMS BRANCH 4.0
END DESCRIPTION:
XS GIS Cut Line= 3
      3817429.17     10494756.29      3816882.29     10494162.54
      3816414.08     10493626.71
#Sta/Elev= 30
  4178.9  334.20  4232.3  332.28  4253.9  333.06  4374.1  328.98  4543.7  316.18
  4614.6  312.42  4678.1  312.03  4911.7  304.71  4954.3  305.37  4968.4  304.67
  4970.6  303.55  4982.6  299.25  4983.1  297.41  4985.9  296.91  4989.1  297.41
  5011.1  302.22  5017.7  304.91  5025.3  304.46  5032.0  306.66  5068.0  303.94
  5074.7  305.09  5124.0  305.37  5145.9  309.52  5160.1  315.51  5181.0  318.48
  5195.2  318.84  5201.9  321.52  5230.3  323.75  5273.1  325.15  5697.7  329.21
#Mann=4,-1,0
  4178.9    0.05       0  4970.6    0.16       0  4983.1    0.07       0
  4989.1    0.16       0
Bank Sta=4983.1,4989.1
Exp/Cntr=0.3,0.1

Type RM Length L Ch R = 1,1344,549,549,549
BEGIN DESCRIPTION:
SIMS BRANCH 3.0
END DESCRIPTION:
XS GIS Cut Line= 3
      3817632.28     10494600.02      3817033.33     10493818.79
      3816627.11     10493391.74
#Sta/Elev= 30
  4297.1  335.50  4435.2  332.30  4505.9  332.47  4611.9  322.17  4790.5  308.66
  4951.6  301.90  4969.1  302.73  4977.3  299.48  4983.6  299.65  4989.9  296.71
  5001.4  294.90  5004.2  294.40  5007.4  294.90  5012.6  299.63  5018.9  302.36
  5212.1  304.84  5268.2  309.81  5284.0  309.75  5290.3  311.68  5325.5  312.70
  5332.8  314.61  5417.6  322.78  5467.1  321.60  5474.0  318.19  5495.4  314.84
  5516.5  319.16  5523.7  321.97  5544.8  323.68  5634.5  323.85  5870.9  329.36
#Mann=5,-1,0
  4297.1    0.05       0  4951.6    0.16       0  5001.4    0.07       0
  5007.4    0.16       0  5634.5    0.05       0
Bank Sta=5001.4,5007.4
Exp/Cntr=0.3,0.1

Type RM Length L Ch R = 1,795,528,528,528
BEGIN DESCRIPTION:
SIMS BRANCH 2.0
END DESCRIPTION:
XS GIS Cut Line= 3
      3817611.47     10494386.55      3817444.79     10493782.34
      3816956.45     10493293.99
#Sta/Elev= 30
  4185.4  330.51  4248.9  330.18  4264.6  328.57  4288.5  328.23  4401.9  318.35
  4589.3  306.06  4771.5  300.98  4909.3  302.27  4951.7  299.78  4958.8  301.97
  4980.0  299.45  4984.1  293.17  4986.8  292.67  4990.1  293.17  5001.2  294.16
  5008.3  297.42  5015.4  299.68  5022.4  299.70  5029.5  301.63  5064.9  300.69
  5079.0  303.25  5086.1  303.09  5093.1  305.61  5114.3  309.39  5121.4  313.01
  5149.7  318.81  5170.9  320.68  5192.1  321.65  5364.8  321.95  5502.8  324.46
#Mann=5,-1,0
  4185.4    0.05       0  4984.1    0.03       0  4990.1    0.05       0
  5008.3    0.16       0  5364.8    0.05       0
Bank Sta=4984.1,4990.1
Exp/Cntr=0.3,0.1

Type RM Length L Ch R = 1,267,0,0,0
BEGIN DESCRIPTION:
SIMS BRANCH 1.0
END DESCRIPTION:
XS GIS Cut Line= 5
      3817637.50     10494303.21      3817689.58     10493771.92
      3817746.88     10493511.50      3817601.04     10493261.50
      3816778.09     10493131.29
#Sta/Elev= 30
  4120.8  327.03  4394.4  313.62  4602.4  306.10  4636.3  306.07  4674.9  303.29
  4772.6  299.21  4914.1  299.04  4957.5  300.24  4992.1  295.45  4999.3  292.27
  5012.4  290.85  5015.2  290.35  5018.4  290.85  5023.1  296.54  5028.9  298.81
  5038.6  299.46  5066.1  298.00  5073.3  298.89  5323.5  299.12  5384.3  303.66
  5434.9  308.76  5441.5  310.31  5536.1  318.43  5586.8  320.11  5634.0  318.93
  5763.5  321.81  5880.4  326.23  5971.5  325.15  6012.0  326.91  6043.9  326.89
#Mann=6,-1,0
  4120.8    0.05       0  4992.1    0.12       0  4999.3    0.16       0
  5012.4    0.07       0  5018.4    0.16       0  5634.0    0.05       0
Bank Sta=5012.4,5018.4
Exp/Cntr=0.3,0.1

Chan Stop Cuts=-1
