--- UNT050 IN BECR.prj (project) ---

Proj Title=UNT050 IN BECR Base Level Engineering
Current Plan=p01
Default Exp/Contr=0.3,0.1
English Units
Geom File=g01
Flow File=f01
Plan File=p01
Y Axis Title=Elevation
X Axis Title(PF)=Main Channel Distance
X Axis Title(XS)=Station
BEGIN DESCRIPTION:
UNT050 IN BECR
END DESCRIPTION:
DSS Export Rating Curves= 0
DSS Export Rating Curve Sorted= 0
DSS Export Volume Flow Curves= 0
DXF OffsetX= 0
DXF OffsetY= 0
DXF ScaleX= 1
DXF ScaleY= 10

--- UNT050 IN BECR.p01 (plan) ---

Plan Title=Multiple Run
Short Identifier=Multiple
Geom File=g01
Flow File=f01
Subcritical Flow
K Sum by GR= 0
Std Step Tol= 0.01
Critical Tol= 0.01
Num of Std Step Trials= 20
Max Error Tol= 0.3
Flow Tol Ratio= 0.001
Split Flow NTrial= 30
Split Flow Tol= 0.02
Split Flow Ratio= 0.02
Log Output Level= 0
Friction Slope Method= 1
Unsteady Friction Slope Method= 2
Unsteady Bridges Friction Slope Method= 1
Parabolic Critical Depth
Global Vel Dist=  1 , 1 , 1
Global Log Level= 0
CheckData=True
Encroach Param= -1, 0, 0, 0
BEGIN DESCRIPTION:
Multiple Run
END DESCRIPTION:

--- UNT050 IN BECR.f01 (steady flow) ---

Flow Title=Multiple
Number of Profiles=7
Profile Names=10-year,25-year,50-year,1pct_min,100-year,1pct_plu,500-year
River Rch & RM= UNT050 IN BECR,Reach-1,27227
     701     959    1176    1059    1433    1937    2134
River Rch & RM= UNT050 IN BECR,Reach-1,19681
     896    1235    1519    1371    1855    2508    2776
River Rch & RM= UNT050 IN BECR,Reach-1,12346
    1455    2039    2536    2310    3124    4225    4761
River Rch & RM= UNT050 IN BECR,Reach-1,5414
    1486    2083    2590    2359    3190    4314    4861
River Rch & RM= UNT050 IN BECR,Reach-1,3602
    1504    2106    2618    2383    3223    4359    4906
Boundary for River Rch & Prof#=UNT050 IN BECR,Reach-1,1
Up Type=0
Dn Type=3
Dn Slope=0.005
Boundary for River Rch & Prof#=UNT050 IN BECR,Reach-1,2
Up Type=0
Dn Type=3
Dn Slope=0.005
Boundary for River Rch & Prof#=UNT050 IN BECR,Reach-1,3
Up Type=0
Dn Type=3
Dn Slope=0.005
Boundary for River Rch & Prof#=UNT050 IN BECR,Reach-1,4
Up Type=0
Dn Type=3
Dn Slope=0.005
Boundary for River Rch & Prof#=UNT050 IN BECR,Reach-1,5
Up Type=0
Dn Type=3
Dn Slope=0.005
Boundary for River Rch & Prof#=UNT050 IN BECR,Reach-1,6
Up Type=0
Dn Type=3
Dn Slope=0.005
Boundary for River Rch & Prof#=UNT050 IN BECR,Reach-1,7
Up Type=0
Dn Type=3
Dn Slope=0.005

--- UNT050 IN BECR.g01 (geometry) ---

Geom Title=Existing Conditions
Program Version=4.10

River Reach=UNT050 IN BECR  ,Reach-1
Reach XY= 30
        3796012.       10504953.      3795854.75       10504862.
       3796147.5       10503899.      3795951.75       10503300.
      3796185.25       10503125.      3795893.75       10502675.
      3796135.25       10502197.       3795617.5       10501330.
       3795921.5       10500767.       3795394.5       10500002.
      3796168.25       10499355.        3796273.       10498153.
       3797243.5       10497337.      3797635.25       10494742.
      3797033.25       10494693.      3796818.75       10494172.
      3796227.25       10493906.      3796331.25       10493634.
        3796109.       10493641.       3796065.5       10493378.
      3795899.25       10493485.        3795756.       10492772.
        3795140.       10491844.        3796016.       10491222.
        3796329.       10491300.      3797226.25       10490514.
       3797446.5       10489955.       3797856.5       10490157.
        3798574.       10488913.      3798679.75       10488271.

Type RM Length L Ch R = 1 ,27227   ,424,424,424
BEGIN DESCRIPTION:
UNT050 IN BECR 51.0
END DESCRIPTION:
XS GIS Cut Line= 3
      3796304.71     10504739.35       3795943.6     10504829.63
      3795627.62     10504791.43
#Sta/Elev= 30
  4570.3  348.94  4668.3  340.33  4680.3  337.54  4716.4  335.73  4730.2  333.14
  4757.6  332.33  4781.7  329.27  4822.9  326.26  4840.1  324.78  4886.5   325.2
  4915.7  323.85  4936.3  325.22  4975.6  323.73  4980.6  323.42  4986.8  319.59
  4993.9  317.35  4996.7  316.85  4999.9  317.35    5007  323.01  5047.3  324.46
  5067.6  323.37  5087.6   326.1  5107.7  335.85  5117.8  342.21  5127.8  344.33
  5178.2  349.46  5208.4  350.87  5226.5  349.05  5231.5  350.87  5260.8  350.68
#Mann= 3 ,-1 , 0
  4570.3     .16       0  4993.9     .07       0  4999.9     .16       0
Bank Sta=4822.9,5087.6
XS Rating Curve= 0 ,0
Exp/Cntr=0.3,0.1

Type RM Length L Ch R = 1 ,26803   ,456,456,456
BEGIN DESCRIPTION:
UNT050 IN BECR 50.0
END DESCRIPTION:
XS GIS Cut Line= 3
      3796283.86     10504617.81      3796099.61     10504510.19
      3795799.62     10504410.19
#Sta/Elev= 30
  4775.1  348.96  4820.3  345.89    4836  343.74  4841.7  341.38  4849.5  340.28
  4857.5  340.47  4863.2  338.03  4878.9  335.09  4894.7  331.18  4900.4  328.31
  4930.6  324.48  4959.1  321.05  4980.6   321.7  4985.6  318.06  4991.1  318.06
    4996  315.76  4998.8  315.26    5002  315.76  5009.6  320.33  5030.6  322.62
  5041.2  323.22  5104.4  322.23  5125.5  324.06  5157.1  326.99  5178.2  331.02
  5209.8  333.66  5220.4  335.21  5230.9  335.21  5283.6  339.94  5304.7  341.15
#Mann= 3 ,-1 , 0
  4775.1     .16       0    4996     .07       0    5002     .16       0
Bank Sta=4930.6,5125.5
XS Rating Curve= 0 ,0
Exp/Cntr=0.3,0.1

Type RM Length L Ch R = 1 ,26347   ,259,259,259
BEGIN DESCRIPTION:
UNT050 IN BECR 49.0
END DESCRIPTION:
XS GIS Cut Line= 3
      3796399.65      10504260.2      3796099.61     10504160.19
      3795799.58     10504160.19
#Sta/Elev= 30
  4688.7  336.55  4699.3  336.32  4741.5  332.14    4752  329.73  4767.8  328.35
  4773.1   326.9  4825.8  321.97  4867.9  320.44  4920.6  321.27  4962.8  320.31
  4983.9  318.74  4991.4  313.61  4994.2  313.11  4997.4  313.61  5002.3  316.13
  5007.5  316.13    5015  318.67    5025  318.29    5055     319    5065   319.6
    5085  322.54    5115  325.93    5125  325.89    5175  330.17    5195  330.54
    5255  336.77    5265  338.59    5295  341.12  5302.5  342.98    5305  342.98
#Mann= 3 ,-1 , 0
  4688.7     .16       0  4991.4     .07       0  4997.4     .16       0
Bank Sta=4825.8,5085
XS Rating Curve= 0 ,0
Exp/Cntr=0.3,0.1

Type RM Length L Ch R = 1 ,26088   ,457,457,457
BEGIN DESCRIPTION:
UNT050 IN BECR 48.0
END DESCRIPTION:
XS GIS Cut Line= 3
      3796592.93     10504034.49      3796016.51     10503989.35
      3795676.22     10504149.08
#Sta/Elev= 30
  4512.4  341.96  4525.8  342.19  4555.9  339.41  4626.1  337.04  4696.3  336.54
  4706.3  334.99  4736.4  333.78  4856.8  320.57  4889.8  318.87  4957.1  319.66
  4997.2  317.57    5016  312.44  5018.8  311.94    5022  312.44  5027.3  318.01
  5057.4  318.25  5077.4  320.09  5098.2  319.58    5104  320.78  5208.7  326.99
  5252.9  332.89  5269.2   333.5    5286  336.76  5337.7  341.19  5343.2  342.66
  5411.7  344.73  5428.9  343.96  5434.5  345.02  5457.3  342.69  5466.5  343.41
#Mann= 3 ,-1 , 0
  4512.4     .16       0    5016     .07       0    5022     .16       0
Bank Sta=4856.8,5104
XS Rating Curve= 0 ,0
Exp/Cntr=0.3,0.1

Type RM Length L Ch R = 1 ,25631   ,255,255,255
BEGIN DESCRIPTION:
Mapping XS c472e84f
END DESCRIPTION:
XS GIS Cut Line= 3
        3796704.     10503853.93      3795901.93      10503732.4
      3795266.49     10503715.04
#Sta/Elev= 30
  4327.1  346.66  4503.5  335.43  4513.6  333.47  4582.5  331.08  4604.6  332.27
  4695.7  325.79  4720.1  326.29  4783.8  322.05  4788.9  323.39  4796.8  321.59
  4852.6   318.3  4897.9  317.72  4990.1  315.44  4999.1  313.45  5019.3  314.67
  5026.4  313.17  5029.2  312.67  5032.4  313.17  5048.8  315.29    5137  317.96
  5390.7  333.81  5399.1  334.59  5404.1  337.01  5500.8  343.47  5580.8  355.58
  5600.8  356.89  5620.8  355.87  5650.8  359.63  5740.9  365.49    5774  369.74
#Mann= 3 ,-1 , 0
  4327.1     .16       0  5026.4     .07       0  5032.4     .16       0
Bank Sta=4897.9,5137
XS Rating Curve= 0 ,0
Exp/Cntr=0.3,0.1

Type RM Length L Ch R = 1 ,25376   ,639,639,639
BEGIN DESCRIPTION:
UNT050 IN BECR 47.0
END DESCRIPTION:
XS GIS Cut Line= 3
      3796439.12     10503641.79      3795673.46      10503469.9
      3795263.27      10503469.9
#Sta/Elev= 30
  4482.1  335.52  4543.1  337.29  4606.6  334.75  4717.3  323.43  4741.7  322.59
  4748.1   320.7  4819.8  316.53  4833.5  316.44  4850.6  313.26  4901.8  313.72
    4912  315.17  4983.8   314.4  5001.3  308.95    5004  308.45  5007.3  308.95
  5011.9  315.17  5024.8   313.8  5045.3  317.16  5103.7  324.43  5243.9  334.32
  5330.7   342.7  5340.7   341.4  5420.7     351  5450.7  357.28  5500.7  359.43
  5560.7  366.87  5580.7  366.36  5600.7  371.21  5670.7  380.14    5677  382.85
#Mann= 3 ,-1 , 0
  4482.1     .16       0  5001.3     .07       0  5007.3     .16       0
Bank Sta=4819.8,5045.3
XS Rating Curve= 0 ,0
Exp/Cntr=0.3,0.1

Type RM Length L Ch R = 1 ,24737   ,636,636,636
BEGIN DESCRIPTION:
UNT050 IN BECR 46.0
END DESCRIPTION:
XS GIS Cut Line= 4
      3796558.84     10503386.55      3796251.58     10503188.65
        3796012.     10503141.78      3795189.11     10503308.44
#Sta/Elev= 30
  4542.4   336.9  4567.3  336.99    4634  332.68  4806.3  325.79  4836.7  322.79
    4971  314.94  4977.1  312.15  4991.4  311.19  4998.6  306.85  5001.3  306.35
  5004.6  306.85    5022  311.44  5033.7  308.85  5042.3  308.92  5052.5  310.97
  5113.7  313.54  5236.1  314.57  5277.6  316.44  5348.3  321.28  5491.1  334.75
  5664.6  345.99    5722  352.47  5777.8  355.99  5797.2  359.67  5817.6     359
  5919.7  370.34  5940.1  373.88  5970.4  375.25  5980.9  378.54  5991.6  379.58
#Mann= 4 ,-1 , 0
  4542.4     .16       0  4998.6     .07       0  5004.6     .16       0
  5277.6      .1       0
Bank Sta=4971,5236.1
XS Rating Curve= 0 ,0
Exp/Cntr=0.3,0.1

Type RM Length L Ch R = 1 ,24101   ,446,446,446
BEGIN DESCRIPTION:
UNT050 IN BECR 45.0
END DESCRIPTION:
XS GIS Cut Line= 3
      3796506.81     10503235.55      3795991.17     10502709.49
      3795105.74     10503120.95
#Sta/Elev= 30
  4167.2   331.2  4324.6  324.79  4395.3  323.12  4402.3  324.33  4536.8  319.89
  4607.5  318.91  4628.6   320.8  4635.8  319.41  4706.5  319.22  4741.8  317.21
  4777.1  312.96  4840.8  310.48  4942.6  310.95    4960  307.82  4993.9   308.2
  5001.8   304.7  5004.5   304.2  5007.8   304.7  5016.8  308.55  5026.8  309.66
  5039.7  309.84  5048.9  308.07  5085.5  308.63  5108.4  311.44  5137.1  313.53
  5192.3  314.25  5357.6  323.59  5514.1  333.58  5679.8  348.16  5880.2  360.49
#Mann= 4 ,-1 , 0
  4167.2     .16       0  5001.8     .07       0  5007.8     .16       0
  5357.6      .1       0
Bank Sta=4840.8,5108.4
XS Rating Curve= 0 ,0
Exp/Cntr=0.3,0.1

Type RM Length L Ch R = 1 ,23655   ,139,139,139
BEGIN DESCRIPTION:
UNT050 IN BECR 44.0
END DESCRIPTION:
XS GIS Cut Line= 2
      3797056.76     10502054.31      3795036.38     10502835.38
#Sta/Elev= 30
  3995.7  364.95  4153.5  357.98  4346.4  337.03  4360.6  332.25  4385.2  332.03
  4390.5  335.58  4446.5  331.72    4541  325.22  4578.7  319.49  4682.5   314.2
  4788.6   312.8  4886.7  309.98  4922.4  303.39  4925.1  302.89  4928.4  303.39
  5020.4  305.28  5025.7  308.52  5064.8   304.3  5104.9  306.66  5110.2  304.27
  5129.1   308.7  5188.3  310.65  5283.8  315.25  5327.9  316.71  5614.2   329.3
  5660.9  333.62    5779  334.69  5865.8   338.9    5939  343.27  6161.8  346.29
#Mann= 13 ,-1 , 0
  3995.7     .16       0  4446.5     .05       0    4541      .1       0
  4682.5     .05       0  4788.6     .16       0  4922.4     .07       0
  4928.4     .16       0  5188.3     .05       0  5283.8     .16       0
  5327.9      .1       0  5614.2     .05       0    5779     .16       0
  5865.8     .05       0
Bank Sta=4886.7,5129.1
XS Rating Curve= 0 ,0
Exp/Cntr=0.3,0.1

Type RM Length L Ch R = 1 ,23516   ,585,585,585
BEGIN DESCRIPTION:
UNT050 IN BECR 43.0
END DESCRIPTION:
XS GIS Cut Line= 2
      3797067.18     10501903.27      3795313.32     10502590.24
#Sta/Elev= 30
  3942.2  366.21  3988.6  361.79    4109   353.2  4122.2  353.98  4163.3  350.92
  4168.7  352.23  4193.1  348.02  4221.7   347.7  4369.2   335.9  4494.3  332.12
  4578.3  327.27  4686.9  327.11  4723.6  324.77  4746.5  320.15    4788  320.29
  4855.1  314.99  4863.2  312.76  4895.4  311.89  4916.9   308.6  4933.8  305.14
    5032  304.84  5034.8  304.34    5038  304.84  5072.1  305.56  5088.7  308.04
  5264.8  311.02  5357.2  317.93  5421.7  319.32  5713.2  341.12  5825.8  347.28
#Mann= 6 ,-1 , 0
  3942.2     .05       0  3988.6     .16       0  4221.7     .05       0
    5032     .04       0    5038     .05       0  5713.2      .1       0
Bank Sta=4916.9,5088.7
XS Rating Curve= 0 ,0
Exp/Cntr=0.3,0.1

Type RM Length L Ch R = 1 ,22931   ,596,596,596
BEGIN DESCRIPTION:
UNT050 IN BECR 42.0
END DESCRIPTION:
XS GIS Cut Line= 2
      3796512.03     10501636.56      3795230.75     10502131.36
#Sta/Elev= 30
  4279.3  334.67  4439.7   329.4  4445.1   328.1  4464.1  329.22  4529.6  326.17
  4548.8  326.64  4584.1  323.76  4603.4  323.78  4614.2  321.78  4638.7  321.69
  4663.3  319.07  4747.8  315.26  4807.7  309.47  4886.9  304.72  4935.8  301.21
  4989.4  301.27  4998.4  298.33  5001.1  297.83  5004.4  298.33  5010.8  302.37
  5020.6  303.54    5026  303.72  5055.9   299.6  5110.5   305.5    5118  304.76
    5195  307.03  5364.6   318.1  5568.3  327.57  5635.2  332.23  5652.8  333.24
#Mann= 4 ,-1 , 0
  4279.3     .16       0  4998.4     .07       0  5004.4     .16       0
  5635.2      .1       0
Bank Sta=4886.9,5110.5
XS Rating Curve= 0 ,0
Exp/Cntr=0.3,0.1

Type RM Length L Ch R = 1 ,22335   ,622,622,622
BEGIN DESCRIPTION:
UNT050 IN BECR 41.0
END DESCRIPTION:
XS GIS Cut Line= 2
      3796431.81     10501465.76      3795306.77     10501637.64
#Sta/Elev= 30
  4414.2  336.17  4425.8  335.23  4456.9  334.35    4467  333.15  4487.2  333.66
  4507.5  331.53  4541.7  331.53  4558.1  331.56  4568.2  329.97  4669.3  323.13
  4679.9  323.47    4730  321.04  4743.4  321.63  4821.1  317.68  4922.2  308.56
  4962.7  303.94  4972.8   300.3  5004.3   296.4    5007   295.9  5010.3   296.4
  5013.3  299.41  5053.7  298.98  5104.3  302.31    5165  301.92  5202.7  298.12
  5225.7  299.08  5256.1  302.15  5357.2     309  5488.7  320.59  5552.3  323.42
#Mann= 5 ,-1 , 0
  4414.2     .16       0  4425.8      .1       0  4541.7     .16       0
  5004.3     .07       0  5010.3     .16       0
Bank Sta=4962.7,5256.1
XS Rating Curve= 0 ,0
Exp/Cntr=0.3,0.1

Type RM Length L Ch R = 1 ,21713   ,554,554,554
BEGIN DESCRIPTION:
UNT050 IN BECR 40.0
END DESCRIPTION:
XS GIS Cut Line= 3
      3795999.57     10501310.18      3795699.61     10501210.19
      3795549.63     10500960.22
#Sta/Elev= 30
    4697  311.07  4823.4  302.15  4865.6  299.83  4886.7  297.15  4907.8  295.93
  4918.3  296.08  4949.9   299.3    4971  299.58  4981.6  296.62  4999.6  294.69
  5002.4  294.19  5005.6  294.69  5010.6  296.47  5026.8     297  5063.7  296.51
  5079.3  295.76  5094.8  295.98  5100.7   295.2  5106.5  295.21    5122  296.73
  5129.8  300.23  5137.6   302.2  5143.4  302.58  5153.1  304.73  5180.3  307.18
  5188.1  308.76  5195.9  308.97  5211.4  311.23  5254.2  315.12  5304.7  319.07
#Mann= 3 ,-1 , 0
    4697     .16       0  4999.6     .07       0  5005.6     .16       0
Bank Sta=4865.6,5129.8
XS Rating Curve= 0 ,0
Exp/Cntr=0.3,0.1

Type RM Length L Ch R = 1 ,21159   ,498,498,498
BEGIN DESCRIPTION:
UNT050 IN BECR 39.0
END DESCRIPTION:
XS GIS Cut Line= 3
      3796199.65     10500710.17      3795899.61     10500860.19
      3795649.57     10500860.19
#Sta/Elev= 30
  4654.4     316  4743.9  308.61  4752.3  306.42  4757.9  306.58  4774.6  303.76
  4788.6  303.53    4797  304.47    4811  303.41  4819.4  301.47  4824.9  301.76
  4855.7  298.77  4864.1  296.73  4869.7  296.84  4908.8  293.31  4914.4  293.91
  4945.1  293.07  4975.9  295.46  4992.4  294.63  4996.9  291.53  4999.6  291.03
  5002.9  291.53  5009.9  294.82  5039.9  294.37  5059.9  295.24  5069.9  297.99
  5119.9  302.71  5129.9  302.77  5139.9  304.52  5179.9  308.77  5239.9  312.83
#Mann= 3 ,-1 , 0
  4654.4     .16       0  4996.9     .07       0  5002.9     .16       0
Bank Sta=4855.7,5069.9
XS Rating Curve= 0 ,0
Exp/Cntr=0.3,0.1

Type RM Length L Ch R = 1 ,20661   ,443,443,443
BEGIN DESCRIPTION:
UNT050 IN BECR 38.0
END DESCRIPTION:
XS GIS Cut Line= 4
      3796215.12     10500386.57      3795777.62     10500511.57
       3795574.5     10500600.11      3795407.84     10500980.31
#Sta/Elev= 30
  4434.8  332.72  4450.9  329.36  4466.3  328.24  4500.1  320.94  4505.3  321.72
  4513.3  319.48  4565.3  313.52  4572.9  310.62  4611.9  307.88  4617.3  305.74
  4658.9  301.01  4731.7  296.95  4864.2   294.2  4909.4  291.93  4985.8  293.26
  4997.6  291.04  5000.3  290.54  5003.6  291.04  5007.6   292.8  5018.5  292.97
  5052.9  291.62  5070.8  294.33  5236.3  300.36    5382  311.68  5395.3   310.5
  5439.7  311.52  5449.9  314.41  5457.6  313.08  5486.4  316.02  5526.5  316.54
#Mann= 3 ,-1 , 0
  4434.8     .16       0  4997.6     .07       0  5003.6     .16       0
Bank Sta=4864.2,5070.8
XS Rating Curve= 0 ,0
Exp/Cntr=0.3,0.1

Type RM Length L Ch R = 1 ,20218   ,537,537,537
BEGIN DESCRIPTION:
UNT050 IN BECR 37.0
END DESCRIPTION:
XS GIS Cut Line= 3
      3796251.57     10500266.78      3795449.61     10500210.19
      3794956.14     10500084.85
#Sta/Elev= 30
  4209.5  331.22  4221.5  331.75  4251.6  326.32  4261.6  326.71  4462.1  304.68
  4572.4  297.74  4657.9  296.46  4702.7   292.3  4799.1  294.68  4873.1  293.87
  4940.3  290.01  4983.4   289.9  4993.4  285.05    5011   290.2  5044.4  291.61
  5054.7  291.31    5065  286.24  5072.3  287.92  5074.5  284.74  5077.2  284.24
  5080.5  284.74  5085.7  286.47  5118.4   286.7    5127  291.24  5154.2  292.34
  5302.4   306.5  5405.5     321  5440.8   324.1  5446.8  326.35  5522.6  331.91
#Mann= 3 ,-1 , 0
  4209.5     .16       0  5074.5     .07       0  5080.5     .16       0
Bank Sta=4702.7,5154.2
XS Rating Curve= 0 ,0
Exp/Cntr=0.3,0.1

Type RM Length L Ch R = 1 ,19681   ,487,487,487
BEGIN DESCRIPTION:
UNT050 IN BECR 36.0
END DESCRIPTION:
XS GIS Cut Line= 3
      3796256.76      10500162.6      3795599.61     10499810.19
      3794959.87      10499839.7
#Sta/Elev= 30
  4211.5  325.83  4270.1  321.09  4276.4  319.02  4412.2  306.85  4423.9  304.63
  4483.7  300.23  4549.5  298.23  4571.4     296  4609.6  297.12  4669.7  293.17
  4855.1  290.82  4921.5  287.26  4949.1  288.02  4954.3  285.82  4959.7  285.82
  4967.2  288.43  4977.2     288  4984.2  281.94    4987  281.44  4990.2  281.94
  4997.2  285.47  5037.3  289.49  5157.4  290.14  5187.4  291.63  5287.6  296.64
  5407.7  307.48  5517.8  323.78  5547.8  325.69  5567.8   329.6  5597.6  331.87
#Mann= 3 ,-1 , 0
  4211.5     .16       0  4984.2     .07       0  4990.2     .16       0
Bank Sta=4855.1,5187.4
XS Rating Curve= 0 ,0
Exp/Cntr=0.3,0.1

Type RM Length L Ch R = 1 ,19194   ,400,400,400
BEGIN DESCRIPTION:
UNT050 IN BECR 35.0
END DESCRIPTION:
XS GIS Cut Line= 3
      3796349.58     10499610.18      3795949.61     10499560.19
      3795549.59     10499310.18
#Sta/Elev= 30
  4582.3  308.68  4723.4  293.48  4743.5  295.44  4753.6  292.72  4773.7  289.73
  4781.3  290.04  4786.3  288.89    4804  289.95  4894.7  286.39  4955.1  286.06
  4975.3  287.04    4993  285.15  4995.9  281.59  4998.7  281.09  5001.9  281.59
  5014.3  287.58  5044.3  286.48  5123.9  286.91  5145.2  285.21  5160.5  291.28
    5203  294.93  5276.1   296.8  5291.4  295.99  5385.7  301.32  5391.6  302.83
    5407  302.19  5412.9  303.74  5443.5  305.77  5449.4  308.64  5457.1  308.93
#Mann= 3 ,-1 , 0
  4582.3     .16       0  4995.9     .07       0  5001.9     .16       0
Bank Sta=4781.3,5160.5
XS Rating Curve= 0 ,0
Exp/Cntr=0.3,0.1

Type RM Length L Ch R = 1 ,18794   ,587,587,587
BEGIN DESCRIPTION:
UNT050 IN BECR 34.0
END DESCRIPTION:
XS GIS Cut Line= 2
      3796687.01      10499424.1      3795614.31     10499189.78
#Sta/Elev= 30
  4481.5  342.31  4524.1  340.61    4568  334.27  4652.9  325.67  4660.9  323.06
    4666  324.07  4709.9  313.95  4724.5  313.06  4758.9  307.01  4796.2  302.64
  4802.8   301.6    4808  298.84  4837.1  298.75  4851.9   295.9  4944.8  288.59
  4993.8  285.43  4997.9  280.36  5000.6  279.86  5003.9  280.36  5011.1  283.92
  5021.3  286.05  5144.2  284.83  5174.5  289.08  5228.7  293.59  5297.7  291.84
  5420.5  298.11  5507.4  306.98  5522.9  311.01  5556.4   314.4  5579.5   320.9
#Mann= 3 ,-1 , 0
  4481.5     .16       0  4997.9     .07       0  5003.9     .16       0
Bank Sta=4944.8,5174.5
XS Rating Curve= 0 ,0
Exp/Cntr=0.3,0.1

Type RM Length L Ch R = 1 ,18207   ,536,536,536
BEGIN DESCRIPTION:
UNT050 IN BECR 33.0
END DESCRIPTION:
XS GIS Cut Line= 3
      3796549.63      10499260.2      3796149.61     10498960.19
      3795749.63      10498660.2
#Sta/Elev= 30
  4489.8  318.95  4497.1  316.65  4539.8  312.53  4561.7  307.71  4589.8  306.18
  4647.1  299.14    4818  286.79  4889.8  283.22  4911.7  284.85  4953.4  284.44
  4961.7  282.68  4976.3  283.08  4982.5   280.5  4986.7  283.08  4997.1  283.11
  5000.4  279.11  5003.1  278.61  5006.4  279.11  5011.7  280.04    5018  284.15
  5132.5  282.88  5147.1   287.4  5153.1  289.46    5168  290.62  5203.4  297.32
  5246.8  301.87  5382.5  310.23  5461.7  321.73  5482.5  322.15  5489.8  324.52
#Mann= 5 ,-1 , 0
  4489.8     .16       0  5000.4     .07       0  5006.4     .16       0
  5153.1      .1       0  5246.8     .05       0
Bank Sta=4818,5147.1
XS Rating Curve= 0 ,0
Exp/Cntr=0.3,0.1

Type RM Length L Ch R = 1 ,17671   ,513,513,513
BEGIN DESCRIPTION:
UNT050 IN BECR 32.0
END DESCRIPTION:
XS GIS Cut Line= 3
      3796599.58     10498910.17      3796199.61     10498610.19
      3795799.64     10498210.22
#Sta/Elev= 30
  4515.3  315.19    4608  306.04  4637.1  301.37  4722.6  295.48    4808  286.27
  4822.6   282.8  4843.4  280.69  4901.7  283.27  4928.8  281.58  4987.1  282.78
  4993.4  281.64  4998.7  278.01  5001.5  277.51  5004.7  278.01  5012.1  283.21
  5029.4  282.63  5100.1  287.72  5114.3  287.77  5128.4  285.75  5169.3  287.13
    5185  283.08  5213.3  286.62  5227.4  287.48  5255.7  293.32    5284  296.63
  5368.8  301.79  5411.2  306.01  5426.4  309.38    5482  317.35  5580.9  337.45
#Mann= 5 ,-1 , 0
  4515.3     .16       0  4998.7     .07       0  5004.7     .16       0
  5169.3      .1       0  5426.4     .05       0
Bank Sta=4808,5213.3
XS Rating Curve= 0 ,0
Exp/Cntr=0.3,0.1

Type RM Length L Ch R = 1 ,17158   ,727,727,727
BEGIN DESCRIPTION:
UNT050 IN BECR 31.0
END DESCRIPTION:
XS GIS Cut Line= 3
      3796699.64     10498660.22      3796299.61     10498260.19
      3795949.64     10498010.21
#Sta/Elev= 30
  4459.5  307.46  4586.8  293.06  4728.2  284.08  4770.7  282.53  4827.2  282.52
  4869.7  279.76  4989.9  281.18  4996.9  280.97  5011.1  277.73  5021.7   281.3
  5028.3   281.3  5047.3  280.65  5053.5  276.43  5059.1  276.26  5061.8  275.76
  5065.1  276.26  5074.4  284.47    5083  286.77  5089.1  285.96  5097.7  288.35
  5131.1  291.17  5182.8  296.73  5197.3   298.3  5204.6  300.46  5261.2  306.28
  5283.3  310.86  5341.1  317.79  5382.8   321.4  5427.1  328.77  5455.3  331.93
#Mann= 5 ,-1 , 0
  4459.5     .16       0  5059.1     .07       0  5065.1     .16       0
  5131.1      .1       0  5182.8     .05       0
Bank Sta=4728.2,5074.4
XS Rating Curve= 0 ,0
Exp/Cntr=0.3,0.1

Type RM Length L Ch R = 1 ,16431   ,657,657,657
BEGIN DESCRIPTION:
UNT050 IN BECR 30.0
END DESCRIPTION:
XS GIS Cut Line= 3
      3796944.28     10498459.47      3796499.61     10497910.19
      3795965.14     10497589.71
#Sta/Elev= 30
  4293.3  338.36  4310.2  336.13  4345.4  321.35  4431.6  306.61    4502  300.98
    4510  302.11  4588.3  297.68  4673.1  289.28  4693.9  285.57  4751.4  282.71
  4836.2  278.14  4978.4  279.04  4993.8   275.1  4996.5   274.6  4999.8   275.1
  5007.8   275.4  5013.6  279.64  5023.3  278.24  5029.2  282.81    5035   284.6
  5145.8  290.44  5204.1  291.82  5212.9  289.72  5225.5  286.22  5241.1  287.06
  5246.9  290.74  5268.3  293.19  5421.8  303.63    5595  323.25  5623.2  325.86
#Mann= 5 ,-1 , 0
  4293.3     .16       0  4993.8     .07       0  4999.8     .16       0
  5212.9      .1       0    5595     .05       0
Bank Sta=4751.4,5029.2
XS Rating Curve= 0 ,0
Exp/Cntr=0.3,0.1

Type RM Length L Ch R = 1 ,15774   ,539,539,539
BEGIN DESCRIPTION:
UNT050 IN BECR 29.0
END DESCRIPTION:
XS GIS Cut Line= 3
      3796999.61     10498410.17      3796849.61     10497610.19
      3796699.59     10497360.16
#Sta/Elev= 30
  4152.4  335.69  4154.9  335.69  4162.6  330.45  4172.7  327.84  4178.7  323.08
  4203.3  315.99  4213.4  314.55    4244  305.62  4283.8  299.89  4446.6  284.53
  4488.1  282.43  4549.2  281.62  4772.2  278.66  4864.6  279.35    4946  276.43
  4969.2  278.69  4989.6  277.67  4998.3  273.03  5001.1  272.53  5004.3  273.03
  5024.6  278.75  5075.2  278.74  5106.3  281.39  5141.3  284.41  5164.6  287.92
  5174.3  291.29  5199.6  295.03  5213.2  299.27  5234.5  302.48  5257.9  303.79
#Mann= 4 ,-1 , 0
  4152.4     .16       0  4998.3     .07       0  5004.3     .16       0
  5174.3      .1       0
Bank Sta=4549.2,5106.3
XS Rating Curve= 0 ,0
Exp/Cntr=0.3,0.1

Type RM Length L Ch R = 1 ,15235   ,393,393,393
BEGIN DESCRIPTION:
UNT050 IN BECR 28.0
END DESCRIPTION:
XS GIS Cut Line= 3
      3797549.62      10497560.2      3797149.61     10497360.19
      3796882.94     10497033.81
#Sta/Elev= 30
  4576.3  305.62  4584.7  303.09  4590.3  303.65  4651.8  294.67  4657.4  295.28
  4665.8  292.79  4696.5  291.28  4732.8  285.27  4785.9   280.2  4808.3  280.63
  4889.4  278.63  4903.3  275.47  4925.7  274.78  4942.5  276.66  4948.1  275.12
  4964.8  277.07  4978.8  276.52  4998.2  271.61  5000.9  271.11  5004.2  271.61
  5009.6   271.9  5015.1  275.58  5020.7  276.37  5065.9  276.88  5115.4  280.26
  5187.2  284.37  5329.4  302.49  5350.2  301.84  5378.9  305.15    5445  306.83
#Mann= 3 ,-1 , 0
  4576.3     .16       0  4998.2     .07       0  5004.2     .16       0
Bank Sta=4808.3,5115.4
XS Rating Curve= 0 ,0
Exp/Cntr=0.3,0.1

Type RM Length L Ch R = 1 ,14842   ,652,652,652
BEGIN DESCRIPTION:
UNT050 IN BECR 27.0
END DESCRIPTION:
XS GIS Cut Line= 3
      3797751.61     10497230.33      3797273.57      10497077.9
       3797074.1     10496928.29
#Sta/Elev= 30
  4557.5  315.65  4601.6  312.81  4607.1  310.87  4644.5  307.56  4654.1  305.03
  4676.7  302.85  4703.7  298.14  4735.9  294.63  4741.1  295.04  4768.1  290.33
  4773.3  290.67    4780  288.28  4853.5  280.26    4870   277.6  4895.5  276.28
    4948  274.88  4979.4  276.62  4989.9  272.95    5001  271.23  5003.8  270.73
    5007  271.23  5010.9  276.47  5058.7  277.26  5102.5  276.48  5160.9  279.56
  5181.7  280.77  5210.9  285.38  5231.7  286.59  5267.1  291.79  5308.6  300.42
#Mann= 3 ,-1 , 0
  4557.5     .16       0    5001     .07       0    5007     .16       0
Bank Sta=4853.5,5160.9
XS Rating Curve= 0 ,0
Exp/Cntr=0.3,0.1

Type RM Length L Ch R = 1 ,14190   ,470,470,470
BEGIN DESCRIPTION:
UNT050 IN BECR 26.0
END DESCRIPTION:
XS GIS Cut Line= 3
      3797799.65     10496660.19      3797449.61     10496660.19
      3796863.66     10496451.33
#Sta/Elev= 30
  4669.1  306.56  4849.1  281.13  4859.1  275.47  4869.1  274.64  4959.1  275.93
  4996.1  269.59  4998.9  269.09  5002.1  269.59  5009.1  272.76  5034.5  275.51
  5090.9  275.58  5096.2  274.17  5114.7  274.95  5121.7   276.8  5208.8  278.47
  5220.9  280.99  5238.3  281.19  5270.5  284.54  5275.8  283.62  5326.8   286.6
  5332.1  288.52    5358  290.57  5393.7  297.29  5475.6  303.95  5486.3  306.25
  5537.2  308.17  5581.8  311.96  5624.3  312.03  5629.6  314.04  5641.2  314.99
#Mann= 5 ,-1 , 0
  4669.1     .16       0  4996.1     .07       0  5002.1     .16       0
  5238.3     .12       0    5358     .16       0
Bank Sta=4849.1,5208.8
XS Rating Curve= 0 ,0
Exp/Cntr=0.3,0.1

Type RM Length L Ch R = 1 ,13720   ,421,421,421
BEGIN DESCRIPTION:
UNT050 IN BECR 25.0
END DESCRIPTION:
XS GIS Cut Line= 3
      3797881.76     10496183.45        3797387.      10496282.4
      3797006.82     10496120.96
#Sta/Elev= 30
  4605.6  326.37  4679.2  322.07  4720.8  311.62  4730.2  304.36  4771.7  294.25
  4822.7  287.28  4883.1  282.65  4903.5  278.81  4919.6  279.07  4944.3  276.67
  4954.5  272.87  4985.1  274.34  4992.3  269.63  4995.1  269.13  4998.3  269.63
  5021.6  273.77  5110.2  274.53  5155.2  276.43  5172.5  279.25  5231.6  286.88
  5255.3  292.92  5260.7  290.95  5302.6  296.31  5331.7  298.01  5337.1  295.95
  5355.3  298.57  5360.8  297.04  5437.2  305.82  5484.5  315.07  5523.2  318.57
#Mann= 3 ,-1 , 0
  4605.6     .16       0  4992.3     .07       0  4998.3     .16       0
Bank Sta=4919.6,5172.5
XS Rating Curve= 0 ,0
Exp/Cntr=0.3,0.1

Type RM Length L Ch R = 1 ,13299   ,455,455,455
BEGIN DESCRIPTION:
UNT050 IN BECR 24.0
END DESCRIPTION:
XS GIS Cut Line= 3
      3797881.75     10496048.01      3797626.58     10495912.61
      3797060.06     10495845.04
#Sta/Elev= 30
  4543.8  320.55  4550.8  320.56  4557.5  318.16  4611.2  314.53  4682.8  312.77
  4737.4  309.45  4859.8  297.09    4880  293.09  4910.2   280.7  4930.3  276.86
  4964.7  273.59  4982.7  273.26  4997.8  270.41  5000.6  269.91  5003.8  270.41
  5010.9  272.23  5060.2  272.37  5101.5  277.54  5131.7  281.82  5147.8  289.71
  5151.9  290.24    5172  295.41  5192.2  298.17  5230.3  300.41  5235.3  299.19
  5312.8  314.96  5317.8   312.9  5323.1  315.34  5343.2  319.13  5403.2  328.41
#Mann= 5 ,-1 , 0
  4543.8     .16       0  4964.7     .12       0  4997.8     .07       0
  5003.8     .12       0  5151.9     .16       0
Bank Sta=4930.3,5101.5
XS Rating Curve= 0 ,0
Exp/Cntr=0.3,0.1

Type RM Length L Ch R = 1 ,12844   ,498,498,498
BEGIN DESCRIPTION:
UNT050 IN BECR 23.0
END DESCRIPTION:
XS GIS Cut Line= 3
      3798078.04     10495843.37        3797427.     10495409.34
      3797027.71     10495548.22
#Sta/Elev= 30
  4362.3  313.84  4398.8  312.03  4470.9  311.22  4514.6  308.28  4568.7  303.84
  4691.8  293.18  4723.3  290.36    4745  285.87  4867.5  275.13  4939.6  272.05
  4984.7  272.41  4997.4  269.53  5005.7  271.17  5011.7  267.79  5017.7  267.68
  5020.5  267.18  5023.7  267.68  5026.7  271.47  5069.5  272.34  5092.8  277.75
  5098.9  278.09  5113.9  283.79  5134.9   284.8  5140.2  288.17  5152.6   290.8
  5213.4  298.12  5284.6  303.53  5377.9  314.12  5432.6  317.42  5567.5  324.46
#Mann= 9 ,-1 , 0
  4362.3     .16       0  4398.8      .1       0  4514.6     .16       0
  4568.7      .1       0  4691.8     .16       0  5017.7     .07       0
  5023.7     .16       0  5213.4     .05       0  5432.6     .16       0
Bank Sta=4867.5,5092.8
XS Rating Curve= 0 ,0
Exp/Cntr=0.3,0.1

Type RM Length L Ch R = 1 ,12346   ,474,474,474
BEGIN DESCRIPTION:
UNT050 IN BECR 22.0
END DESCRIPTION:
XS GIS Cut Line= 3
      3797899.57     10494860.21      3797549.61     10495060.19
      3797199.64     10495360.16
#Sta/Elev= 30
  4632.3  308.12  4660.6  305.85  4699.2  299.87  4712.9  295.23  4720.8  290.21
  4735.9  287.42  4742.4  283.05  4793.5  274.09  4816.2  272.54  4816.5  272.52
  4941.1  271.86  4954.7  273.74  4962.7  271.43  4968.4  273.25  4997.1  264.62
  4999.8  264.12  5003.1  264.62  5012.3  269.29  5032.5  271.79  5134.7  270.57
  5177.5  272.61  5290.6  278.89    5397   292.1  5411.3   292.1  5417.9  294.63
  5425.6  294.21  5446.4  298.46  5454.1   298.1  5460.7  300.98  5496.3  303.44
#Mann= 5 ,-1 , 0
  4632.3     .05       0  4660.6     .16       0  4816.2     .05       0
  4997.1     .03       0  5003.1     .05       0
Bank Sta=4816.5,5177.5
XS Rating Curve= 0 ,0
Exp/Cntr=0.3,0.1

Type RM Length L Ch R = 1 ,11872   ,486,486,486
BEGIN DESCRIPTION:
UNT050 IN BECR 21.0
END DESCRIPTION:
XS GIS Cut Line= 3
      3797849.58     10494710.19      3797599.61     10494710.19
      3796899.61     10495060.19
#Sta/Elev= 30
  4750.4  307.21  4790.4  299.98  4800.4  295.36  4840.4  286.25  4880.4  280.11
  4910.4  277.85  4919.9  274.73  4940.4  274.82  4950.4  271.49  4970.4  269.75
  4990.4  262.93  4994.9   262.8  4997.6   262.3  5000.9   262.8  5003.2   262.8
  5014.4  270.46  5075.8  271.38  5081.4  268.19  5089.8  270.45  5129.5  270.69
  5447.6  269.55  5492.3  272.07  5511.4  273.95  5545.4  277.76  5595.7  291.64
  5604.1  295.71  5665.3  305.53  5680.6  307.38  5729.9  314.27    5783  318.66
#Mann= 8 ,-1 , 0
  4750.4     .05       0  4919.9     .16       0  4994.9     .07       0
  5000.9     .16       0  5129.5     .05       0  5511.4     .16       0
  5665.3     .05       0  5680.6      .1       0
Bank Sta=4940.4,5492.3
XS Rating Curve= 0 ,0
Exp/Cntr=0.3,0.1

Type RM Length L Ch R = 1 ,11386   ,560,560,560
BEGIN DESCRIPTION:
UNT050 IN BECR 20.0
END DESCRIPTION:
XS GIS Cut Line= 3
      3797249.61     10494260.18      3797199.61     10494660.19
      3796899.61     10495010.19
#Sta/Elev= 30
  4661.6  306.92  4752.3  299.98    4780  293.08  4785.1  294.97  4792.6  293.06
  4832.9  280.03    4843  275.39  4860.6  276.03  4865.7  274.26  4903.5  271.62
  4941.3  268.68    4974  268.76  4984.1  266.96  4991.2  261.02  4993.9  260.52
  4997.2  261.02  5021.9  268.57  5026.9  264.72  5044.6  268.39  5062.2  269.01
  5227.7  268.38  5268.7  271.04  5277.1  271.78  5319.9  279.54  5334.2     285
  5348.4  288.17  5405.5  297.16  5454.9  307.07  5517.2  314.49  5525.7  315.96
#Mann= 5 ,-1 , 0
  4661.6     .05       0  4991.2     .03       0  4997.2     .05       0
  5268.7     .16       0  5517.2      .1       0
Bank Sta=4903.5,5277.1
XS Rating Curve= 0 ,0
Exp/Cntr=0.3,0.1

Type RM Length L Ch R = 1 ,10826   ,438,438,438
BEGIN DESCRIPTION:
UNT050 IN BECR 19.0
END DESCRIPTION:
XS GIS Cut Line= 3
      3797209.94     10494245.92      3796913.04     10494475.11
      3796720.81     10494906.33
#Sta/Elev= 30
  4754.7  303.95  4771.6   302.7  4843.6  295.64  4871.6  290.48  4879.8  286.95
  4894.1  284.31  4921.4  275.18  4944.1   271.5  4950.4  268.95  4964.9  267.15
  4985.7  267.88  4997.2  260.08    5000  259.58  5003.2  260.08  5007.8  260.99
  5014.7   267.4    5021  266.79  5029.2  268.39  5174.3  268.81    5244  267.43
  5255.8  267.82  5266.7  272.39  5276.6   274.5  5301.4  279.59  5310.5   280.1
  5319.2  282.57  5382.3  291.74  5492.7  304.95  5573.4  313.18  5601.9  314.92
#Mann= 6 ,-1 , 0
  4754.7     .05       0  4771.6     .16       0  4997.2     .07       0
  5003.2     .16       0  5276.6      .1       0  5382.3     .05       0
Bank Sta=4944.1,5266.7
XS Rating Curve= 0 ,0
Exp/Cntr=0.3,0.1

Type RM Length L Ch R = 1 ,10388   ,518,518,518
BEGIN DESCRIPTION:
UNT050 IN BECR 18.0
END DESCRIPTION:
XS GIS Cut Line= 3
      3796849.61     10493960.17      3796799.61     10494160.19
       3796399.6      10494510.2
#Sta/Elev= 30
  4789.8  306.07  4841.4   297.8  4849.1  293.89  4890.3  283.99  4965.1  270.44
  4977.9  268.57  4993.4  260.31  5000.1  259.51  5002.8  259.01  5006.1  259.51
  5009.7  261.25  5017.3  260.24    5024  266.88  5031.6  264.74  5038.2   267.1
  5109.4  265.98    5116  267.12  5123.6  265.33  5130.3  267.17    5173  265.79
    5218  266.54  5231.3  267.74  5272.6   270.8  5328.6  276.54  5364.7  281.92
  5371.4   281.6  5449.2  293.06  5456.8  295.57  5491.9  298.89  5527.5  304.38
#Mann= 5 ,-1 , 0
  4789.8     .16       0  5000.1     .07       0  5006.1     .16       0
    5218      .1       0  5231.3     .05       0
Bank Sta=4965.1,5272.6
XS Rating Curve= 0 ,0
Exp/Cntr=0.3,0.1

Type RM Length L Ch R = 1 ,9870    ,568,568,568
BEGIN DESCRIPTION:
UNT050 IN BECR 17.0
END DESCRIPTION:
XS GIS Cut Line= 3
      3796799.58      10493910.2      3796399.61     10494060.19
      3796168.25     10494381.36
#Sta/Elev= 30
  4566.9  295.08    4582  292.98  4588.2  289.01  4598.9  287.77  4606.9  284.28
  4684.3  271.11  4692.4  268.91    4728  266.15  4972.7  266.66  4991.4  260.44
  4997.2  260.44  4998.4     258  5001.2   257.5  5004.4     258  5007.6  264.81
  5022.3  266.72  5051.7  266.86  5066.5  269.26  5080.3  270.87  5104.3  276.88
  5122.4  278.43  5129.6  281.23  5152.4  286.28  5158.5  286.46  5166.6   289.1
  5223.6  296.01  5238.3  298.96  5244.4  297.93  5265.3  299.38  5389.9  310.05
#Mann= 4 ,-1 , 0
  4566.9     .16       0  4998.4     .07       0  5004.4     .16       0
  5104.3     .05       0
Bank Sta=4684.3,5066.5
XS Rating Curve= 0 ,0
Exp/Cntr=0.3,0.1

Type RM Length L Ch R = 1 ,9302    ,488,488,488
BEGIN DESCRIPTION:
UNT050 IN BECR 16.0
END DESCRIPTION:
XS GIS Cut Line= 3
      3796697.36     10493392.87      3796299.61     10493710.19
      3795899.62     10494010.18
#Sta/Elev= 30
  4510.6  329.52  4607.1  326.01  4677.5  320.33    4692  318.04  4706.4  311.47
  4720.8  308.44  4741.6  308.14  4749.6  303.87    4756  305.66  4763.6  303.91
  4791.2  296.07  4840.9  276.49  4904.9   268.7  4933.7  262.47    4969  262.71
    4974  255.75  4976.7  255.25    4980  255.75  4983.4  263.79  4991.4  259.49
  4997.8  260.81  5005.8  255.79  5016.2  261.71  5041.3  265.29  5305.9  265.09
    5333  267.76  5391.3  275.62  5426.7  285.17  5477.9  294.45  5519.4  299.28
#Mann= 4 ,-1 , 0
  4510.6     .16       0    4974     .07       0    4980     .16       0
  5477.9     .05       0
Bank Sta=4904.9,5333
XS Rating Curve= 0 ,0
Exp/Cntr=0.3,0.1

Type RM Length L Ch R = 1 ,8814    ,509,509,509
BEGIN DESCRIPTION:
UNT050 IN BECR 15.0
END DESCRIPTION:
XS GIS Cut Line= 3
      3796648.82     10493253.94      3796121.01     10493455.35
      3795537.67     10494038.68
#Sta/Elev= 30
  4402.5  335.75  4491.4  337.23  4691.2  322.99    4716  315.35  4722.8  309.24
  4733.5  307.34  4746.1  300.12  4800.9  281.23  4808.4  277.02  4855.7  267.01
  4915.8  261.94  4978.9  264.89    4986  263.32  4993.1  256.25  4997.1  254.97
  4999.9  254.47  5003.1  254.97  5021.3  262.88  5035.5  264.03  5191.1  262.23
  5247.6  266.29    5283  270.42  5318.3  277.81  5325.4  277.31  5360.8   286.5
    5389  290.58  5466.8   296.8  5551.7  299.36    5699  309.01  5792.4  313.21
#Mann= 4 ,-1 , 0
  4402.5     .16       0  4997.1     .07       0  5003.1     .16       0
    5699     .05       0
Bank Sta=4855.7,5247.6
XS Rating Curve= 0 ,0
Exp/Cntr=0.3,0.1

Type RM Length L Ch R = 1 ,8305    ,559,559,559
BEGIN DESCRIPTION:
UNT050 IN BECR 14.0
END DESCRIPTION:
XS GIS Cut Line= 3
      3796459.95      10492917.8      3795829.71     10493350.11
      3795444.46     10493870.71
#Sta/Elev= 30
  4252.5  318.65  4319.1  308.03    4334  308.54  4340.1  304.41  4369.9  304.89
  4398.4  298.09  4420.6   297.1  4426.7  293.74  4447.7  291.42  4477.5  290.81
  4743.5  264.62  4794.2  260.83  4980.5  262.62  4988.5  260.96  5000.4  253.39
  5003.1  252.89  5006.4  253.39  5019.9  257.01  5030.4  263.11  5130.6  262.22
  5174.5  265.92  5195.3  267.96  5239.2  279.48  5253.2  280.03  5260.1   284.5
  5266.3  283.03  5289.3  286.93  5410.4   291.6  5481.3  287.64  5664.4  305.42
#Mann= 3 ,-1 , 0
  4252.5     .16       0  5000.4     .07       0  5006.4     .16       0
Bank Sta=4743.5,5174.5
XS Rating Curve= 0 ,0
Exp/Cntr=0.3,0.1

Type RM Length L Ch R = 1 ,7746    ,423,423,423
BEGIN DESCRIPTION:
UNT050 IN BECR 13.0
END DESCRIPTION:
XS GIS Cut Line= 3
      3796877.93     10492872.01      3795749.61     10492910.19
      3795122.84     10493079.85
#Sta/Elev= 30
  3842.9  323.69  4041.3  330.24  4211.4  327.22  4281.5  320.51  4361.5  322.05
  4381.5  320.22  4431.6  301.85  4491.6  285.22  4591.7  270.53  4641.7  264.74
  4671.7  263.38  4861.8  259.49  4951.9     261  4974.5  258.79  4982.2  257.06
  4986.2  253.52    4989  253.02  4992.2  253.52  5002.9  253.71  5013.3   258.5
  5029.1  261.34  5127.3  259.48  5210.1  263.69  5251.6  272.76  5257.8  275.81
  5282.7  281.67  5332.4  288.82  5412.1  294.95  5446.8  299.36  5621.2  305.64
#Mann= 3 ,-1 , 0
  3842.9     .16       0  4986.2     .07       0  4992.2     .16       0
Bank Sta=4671.7,5210.1
XS Rating Curve= 0 ,0
Exp/Cntr=0.3,0.1

Type RM Length L Ch R = 1 ,7323    ,461,461,461
BEGIN DESCRIPTION:
UNT050 IN BECR 12.0
END DESCRIPTION:
XS GIS Cut Line= 3
        3796121.     10492045.63      3795599.61     10492560.19
      3794780.75      10493309.5
#Sta/Elev= 30
  4257.8  296.02  4588.6  300.51  4679.2  296.02  4728.7  286.52  4735.8  289.37
  4764.1  288.86  4771.1  285.83  4792.4  288.36  4799.4  284.79  4806.5  287.48
  4813.6  283.74  4834.8  284.11  4841.8  279.95    4849  282.11  4877.2  274.02
  4884.3  268.71  4905.5  265.92  4912.6  261.72  4933.8  259.77  4966.1  250.64
  4968.9  250.14  4972.1  250.64  4993.7  253.97  5004.2  260.49  5237.9  258.69
  5302.1  262.82  5457.5  295.07  5783.1  310.14  6021.8  316.22  6100.3  316.42
#Mann= 5 ,-1 , 0
  4257.8      .1       0  4588.6     .16       0  4966.1     .07       0
  4972.1     .16       0  6021.8      .1       0
Bank Sta=4905.5,5302.1
XS Rating Curve= 0 ,0
Exp/Cntr=0.3,0.1

Type RM Length L Ch R = 1 ,6862    ,337,337,337
BEGIN DESCRIPTION:
UNT050 IN BECR 11.0
END DESCRIPTION:
XS GIS Cut Line= 3
      3795741.12     10492126.49      3795100.97     10492332.64
      3794699.51     10492614.75
#Sta/Elev= 30
  4526.7  295.79  4596.6  296.94  4683.1  294.09  4752.5  294.59  4784.6  292.06
  4816.6   288.5  4843.4  281.92  4848.7  282.38    4875  274.28  4880.8  270.71
    4938  262.72  4944.9  260.99  4982.2  258.63    5001  258.81    5006  250.89
  5008.8  250.39    5012  250.89  5014.3   257.6  5041.1   259.2  5213.1  256.78
  5234.9  258.67  5249.8  257.88    5262   260.2  5327.3  261.02  5384.2  269.15
  5392.7  272.78  5464.1  289.29  5520.8  297.87  5579.8  302.29  5689.9  305.43
#Mann= 4 ,-1 , 0
  4526.7      .1       0  4596.6     .16       0    5006     .07       0
    5012     .16       0
Bank Sta=4938,5327.3
XS Rating Curve= 0 ,0
Exp/Cntr=0.3,0.1

Type RM Length L Ch R = 1 ,6525    ,675,675,675
BEGIN DESCRIPTION:
UNT050 IN BECR 10.0
END DESCRIPTION:
XS GIS Cut Line= 2
      3796002.97     10491955.35      3794032.66     10492052.47
#Sta/Elev= 30
  4191.3  294.07  4244.7  293.25  4424.9  296.02  4543.2  294.73  4605.2  287.24
  4665.2  275.18  4715.3  269.28  4745.3  263.91  4798.9  259.41  4855.5   256.9
  4945.6   258.3  4985.6   254.1  4992.6  250.05  4995.3  249.55  4998.6  250.05
  5005.6  250.45  5015.7  257.87  5025.7   258.4  5155.8  256.36    5286  260.24
  5356.1  265.39  5416.1  272.04  5476.2  280.36  5516.3  288.62  5556.3  293.03
  5656.4  300.11  5760.1  305.33  5866.7  312.19  6156.7  318.17    6164  318.34
#Mann= 6 ,-1 , 0
  4191.3      .1       0  4543.2     .16       0  4992.6     .07       0
  4998.6     .16       0  5760.1      .1       0  6156.7     .16       0
Bank Sta=4798.9,5286
XS Rating Curve= 0 ,0
Exp/Cntr=0.3,0.1

Type RM Length L Ch R = 1 ,5850    ,436,436,436
BEGIN DESCRIPTION:
UNT050 IN BECR 9.0
END DESCRIPTION:
XS GIS Cut Line= 3
      3795795.43     10491811.82      3795499.61     10491610.19
      3794699.63      10491060.2
#Sta/Elev= 30
  4631.7  293.31  4709.3  292.97  4772.8  291.41  4832.4  284.95  4889.4  272.95
  4895.5  269.16  4925.3  261.17  4953.4  256.84  4992.7  255.13  4997.1  254.03
  5000.2  248.23    5003  247.73  5006.2  248.23  5018.1   254.8  5026.1  256.07
  5097.3  254.87  5161.5  253.15  5220.3  256.03  5256.7  253.08  5334.7   256.9
    5493  263.38  5579.6  273.39  5600.6  272.91  5615.5  276.29  5636.5  275.44
  5703.4  280.64  5723.1  280.18  5730.2  281.99  5881.4  292.31  5960.5  300.83
#Mann= 7 ,-1 , 0
  4631.7     .05       0  4709.3     .16       0  5000.2     .07       0
  5006.2     .16       0  5097.3     .05       0  5703.4     .16       0
  5730.2     .05       0
Bank Sta=4953.4,5334.7
XS Rating Curve= 0 ,0
Exp/Cntr=0.3,0.1

Type RM Length L Ch R = 1 ,5414    ,261,261,261
BEGIN DESCRIPTION:
UNT050 IN BECR 8.0
END DESCRIPTION:
XS GIS Cut Line= 3
      3795936.47     10491768.37      3795849.61     10491360.19
      3795249.59     10490660.17
#Sta/Elev= 30
    4591  292.34  4732.3  289.14  4790.5  285.78  4834.5  284.44  4839.9  282.44
  4875.4  278.52  4906.1  269.91  4967.4  258.42  4977.7  258.01  4988.6  250.44
  4995.1  247.78  4997.8  247.28  5001.1  247.78  5011.6  249.17  5015.5  252.57
  5029.7  254.92  5105.7  253.74    5157  252.44    5179  254.64  5334.8   252.4
  5490.7  255.11  5632.3  264.59  5710.2  272.72  5810.1  285.38  5830.9  289.47
  5859.5  291.84  5880.3  297.12  5902.3  300.47  5908.9  304.23  5930.3  305.72
#Mann= 5 ,-1 , 0
    4591     .05       0  4790.5     .16       0  4995.1     .07       0
  5001.1     .16       0  5105.7     .05       0
Bank Sta=4977.7,5490.7
XS Rating Curve= 0 ,0
Exp/Cntr=0.3,0.1

Type RM Length L Ch R = 1 ,5153    ,569,569,569
BEGIN DESCRIPTION:
UNT050 IN BECR 7.0
END DESCRIPTION:
XS GIS Cut Line= 2
      3796044.62     10491740.08      3796072.38     10490234.14
#Sta/Elev= 30
  4479.7  292.92  4619.6  290.29  4694.8  285.89  4719.6  284.96  4769.6  279.15
  4859.7  260.53  4889.7  255.64  4899.7  255.47  4909.7   252.8  4919.7     254
  4944.6  253.89  4979.7  252.84  4986.7  246.36  4989.4  245.86  4992.7  246.36
  4999.7  246.42  5018.2  252.64  5029.7  253.32  5219.7   251.5  5269.7     253
  5359.7  252.12  5439.8   253.8  5529.8  255.82  5679.8  263.71  5719.8  263.88
  5809.8   271.8  5829.8   273.1  5839.8   271.6  5849.8  272.35  5985.9  283.94
#Mann= 5 ,-1 , 0
  4479.7     .05       0  4694.8     .16       0  4944.6     .05       0
  4986.7     .03       0  4992.7     .05       0
Bank Sta=4899.7,5439.8
XS Rating Curve= 0 ,0
Exp/Cntr=0.3,0.1

Type RM Length L Ch R = 1 ,4584    ,497,497,497
BEGIN DESCRIPTION:
UNT050 IN BECR 6.0
END DESCRIPTION:
XS GIS Cut Line= 3
       3796384.9     10491885.87      3796530.73     10491253.96
      3796398.79     10490448.41
#Sta/Elev= 30
  4234.7  293.69  4254.9  292.23  4458.5  292.25    4544   284.7  4599.7  282.83
    4651  275.26  4671.6  267.67  4677.4   262.7  4692.1   262.2  4720.2  255.75
  4768.1  253.14  4819.9   252.2  4976.4   249.1  4983.1  247.17  4985.4   243.6
  4988.1   243.1  4991.4   243.6  5018.8  246.93  5044.5  245.83  5049.5  249.49
  5079.6  246.47  5120.1  252.33  5130.2  257.58  5160.6  264.62  5167.1  268.74
  5172.2  266.74    5191  271.52  5387.6  280.95  5540.2  283.72  5699.5   290.6
#Mann= 7 ,-1 , 0
  4234.7      .1       0  4254.9     .16       0  4819.9     .05       0
  4976.4     .16       0  4985.4     .07       0  4991.4     .16       0
  5387.6     .05       0
Bank Sta=4768.1,5130.2
XS Rating Curve= 0 ,0
Exp/Cntr=0.3,0.1

Type RM Length L Ch R = 1 ,4087    ,307,307,307
BEGIN DESCRIPTION:
UNT050 IN BECR 5.0
END DESCRIPTION:
XS GIS Cut Line= 3
      3796939.08     10491735.51      3796855.75     10490855.32
      3796600.53     10490298.01
#Sta/Elev= 30
  4010.2  288.39  4077.4  288.78  4146.1  291.19  4256.6  287.81  4286.8  283.09
    4347  281.75  4357.1  280.33  4384.8  270.24  4407.3  261.55  4427.4  256.85
  4447.5  252.89  4477.3  251.69  4728.7  249.13  4797.2  251.14  4928.5  249.86
    4977  250.35    4996  243.46  4998.7  242.96    5002  243.46    5010  243.51
  5021.8  250.24  5085.3  252.05  5108.3  253.88  5113.8  256.63  5136.8  259.68
  5142.3   264.4  5159.9  266.03  5211.4  280.83  5400.9  288.91  5507.3  289.34
#Mann= 7 ,-1 , 0
  4010.2     .05       0  4077.4     .16       0  4384.8     .05       0
  4928.5     .16       0    4996     .07       0    5002     .16       0
  5211.4     .05       0
Bank Sta=4477.3,5085.3
XS Rating Curve= 0 ,0
Exp/Cntr=0.3,0.1

Type RM Length L Ch R = 1 ,3780    ,178,178,178
BEGIN DESCRIPTION:
UNT050 IN BECR 4.0
END DESCRIPTION:
XS GIS Cut Line= 4
        3797012.     10491620.99      3797090.12      10490532.4
      3797069.29     10490313.65      3796944.53     10489965.35
#Sta/Elev= 30
  4007.1  292.66  4183.3  281.82  4250.9  269.21  4358.8  254.44  4545.1  250.25
  4559.3  250.15  4598.4  249.54  4603.4  247.81  4639.5  249.58  4741.3  249.41
  4839.4   249.6  4937.5   249.3  4982.8  249.59  5000.4  246.58  5010.5   242.2
  5020.5  241.62  5023.2  241.12  5026.5  241.62  5040.6  249.03  5050.6   250.1
  5251.4  247.69  5365.7  249.74  5421.9   253.7  5470.6  254.25  5502.5  258.65
  5508.9  262.64  5570.4  272.64  5595.9  278.86  5649.9  286.41  5688.2  288.02
#Mann= 10 ,-1 , 0
  4007.1     .16       0  4250.9     .05       0  4545.1     .08       0
  4741.3     .05       0  4839.4     .08       0  4937.5     .05       0
  4982.8     .16       0  5020.5     .07       0  5026.5     .16       0
  5649.9     .05       0
Bank Sta=4559.3,5365.7
XS Rating Curve= 0 ,0
Exp/Cntr=0.3,0.1

Type RM Length L Ch R = 1 ,3602    ,1759,1759,1759
BEGIN DESCRIPTION:
UNT050 IN BECR 3.0
END DESCRIPTION:
XS GIS Cut Line= 6
      3797100.54     10491777.22      3797173.46     10491084.49
      3797230.75     10490563.65      3797183.87     10490350.11
      3797235.96     10490042.82      3797029.05     10489944.54
#Sta/Elev= 30
  3733.5  300.51  3774.1   300.6  3948.7  280.59  3971.8  280.13  4042.2  271.93
  4102.6  260.73  4112.6   261.8  4156.2  257.26  4213.2  254.59  4425.5  252.22
  4514.9  249.29  4726.1   248.6  4917.3  247.23  4967.8  248.95  4977.8  247.95
  4988.3  241.96  4995.5  241.74  4998.3  241.24  5001.5  241.74  5026.7  249.39
  5049.7  249.84  5119.4  246.76  5131.6  248.41  5446.4  248.63    5505  252.88
  5527.8  252.38  5543.9  259.13  5595.9  266.88  5664.1  281.57  5713.4  284.49
#Mann= 6 ,-1 , 0
  3733.5     .05       0  3948.7     .16       0  4425.5     .05       0
  4995.5     .04       0  5001.5     .05       0  5543.9     .16       0
Bank Sta=4726.1,5446.4
XS Rating Curve= 0 ,0
Exp/Cntr=0.3,0.1
