HEC-RAS study UNT094 IN BECR.prj: UNT094 IN BECR Base Level Engineering

--- UNT094 IN BECR.g01 (geometry) --- (continued)

Type RM Length L Ch R = 1 ,36581   ,903,903,903
BEGIN DESCRIPTION:
UNT094 IN BECR 55.0
END DESCRIPTION:
XS GIS Cut Line= 3
      3778449.59     10560360.22      3778149.61     10560960.19
      3777999.62     10561110.18
#Sta/Elev= 30
  4372.4  353.68  4565.2  339.73  4573.6  336.03    4596  331.73  4604.4  332.76
  4649.1  326.47  4760.9  321.11  4783.2  318.09    4828  319.59    4923  317.27
  4931.4  319.26  4945.4  318.64  4953.7  314.81  4962.1  319.87  4967.7  314.24
  4976.1  319.84  4984.5  318.15  4990.1  313.77  5003.9  313.15  5006.6  312.65
  5009.9  313.15  5020.8   314.7  5029.2   313.5  5034.8  316.62  5040.4  313.58
  5046.7  313.58  5057.3  317.92  5071.5  319.46  5085.6  323.44  5255.3  336.52
#Mann= 3 ,-1 , 0
  4372.4     .16       0  5003.9     .07       0  5009.9     .16       0
Bank Sta=4976.1,5085.6
XS Rating Curve= 0 ,0
Exp/Cntr=0.3,0.1

Type RM Length L Ch R = 1 ,35678   ,499,499,499
BEGIN DESCRIPTION:
UNT094 IN BECR 54.0
END DESCRIPTION:
XS GIS Cut Line= 3
       3777799.6     10560060.22      3777649.61     10560660.19
      3777849.59     10561010.15
#Sta/Elev= 30
    4362  355.46  4388.3  352.54  4434.1  348.14  4462.5  342.28    4496  339.57
  4516.6   331.7  4632.5  321.78  4681.5  319.95  4709.9  323.41  4743.4  324.27
  4846.4  320.01  4879.9   316.4  4928.9   316.8  4939.2   310.9  4946.5   310.2
  4949.3   309.7  4952.5   310.2  4957.2  310.34  4962.4  314.98  4983.3  314.89
  4994.1  310.89  5003.5  310.47  5009.9  310.91  5015.7  315.58  5031.5  318.54
  5047.4  315.97  5084.1  316.93  5096.3  319.54    5187  320.45  5383.5   333.3
#Mann= 4 ,-1 , 0
    4362     .05       0  4388.3     .16       0  4946.5     .07       0
  4952.5     .16       0
Bank Sta=4928.9,4962.4
XS Rating Curve= 0 ,0
Exp/Cntr=0.3,0.1

Type RM Length L Ch R = 1 ,35179   ,459,459,459
BEGIN DESCRIPTION:
UNT094 IN BECR 53.0
END DESCRIPTION:
XS GIS Cut Line= 3
       3777499.6     10559960.21      3777349.61     10560510.19
      3776649.62     10561210.18
#Sta/Elev= 30
  4442.4  354.73  4475.2  353.57  4539.1   347.7    4629  332.64    4648  327.68
  4653.1  329.86    4660  325.72  4687.7  322.19  4692.9  323.33  4722.2  320.16
  4767.2  321.09  4846.6  315.92    4971  316.53  4999.1   310.5  5001.9     310
  5005.1   310.5    5016   311.8  5026.6  315.98  5097.3  318.03    5168  314.97
    5267  317.69    5465   317.4  5535.7  319.75  5578.2  318.31  5691.3  320.43
  5832.7  327.92  5917.6  338.15  5931.7  334.04    5960  342.49  6002.4  344.59
#Mann= 4 ,-1 , 0
  4442.4     .05       0  4475.2     .16       0  4999.1     .07       0
  5005.1     .16       0
Bank Sta=4971,5026.6
XS Rating Curve= 0 ,0
Exp/Cntr=0.3,0.1

Type RM Length L Ch R = 1 ,34720   ,482,482,482
BEGIN DESCRIPTION:
UNT094 IN BECR 52.0
END DESCRIPTION:
XS GIS Cut Line= 3
      3777399.58     10559960.21      3776949.61     10560360.19
      3776349.58     10560860.21
#Sta/Elev= 30
  4425.4  350.82  4428.7  350.82    4466  346.23  4558.4  335.67  4638.2  324.65
    4716  319.49  4730.2  315.82  4832.3  315.72  4857.3  314.05    4879  315.94
  4899.9  313.16  4920.8  316.64  4969.3  316.07  4996.4  310.52  4999.2  310.02
  5002.4  310.52  5024.1  315.87  5048.9  313.95  5162.2  316.14  5176.5  311.54
  5212.2  315.57  5285.6   317.9  5311.9  315.72  5410.7  316.95  5453.8  319.58
  5460.3  317.25  5499.8  318.88  5595.6  322.99  5806.1   339.9  5808.5   339.9
#Mann= 13 ,-1 , 0
  4425.4     .05       0  4428.7     .16       0    4466     .12       0
  4558.4     .16       0  4832.3     .12       0  4969.3     .16       0
  4996.4     .07       0  5002.4     .16       0  5212.2     .12       0
  5285.6     .16       0  5410.7     .12       0  5499.8     .16       0
  5806.1     .05       0
Bank Sta=4969.3,5024.1
XS Rating Curve= 0 ,0
Exp/Cntr=0.3,0.1

Type RM Length L Ch R = 1 ,34238   ,439,439,439
BEGIN DESCRIPTION:
UNT094 IN BECR 51.0
END DESCRIPTION:
XS GIS Cut Line= 3
      3777249.61     10559710.19      3776649.61     10560110.19
      3776249.62     10560110.19
#Sta/Elev= 30
  4309.8  351.47  4353.4  348.85  4374.4  348.43  4439.8  342.73  4495.8  336.85
  4620.8  321.46  4692.9  316.64  4738.1  315.48    4771  315.05  4814.6  312.21
  4958.8   314.6  4963.2  312.39  4966.3  310.83  4972.3  312.65  4981.3  309.12
  4987.3  310.09  4994.9  308.33  5002.4  310.34  5005.4  308.32  5008.1  307.82
  5011.4  308.32  5017.4  313.19  5060.9  315.51  5120.9  313.78  5162.1   314.1
  5230.9   318.3  5290.9  326.32  5320.9  327.57  5390.9  334.58  5430.9  335.95
#Mann= 9 ,-1 , 0
  4309.8     .16       0  4353.4     .12       0  4439.8     .16       0
  4495.8     .12       0  4738.1     .16       0  4963.2     .12       0
  5005.4     .07       0  5011.4     .12       0  5162.1     .16       0
Bank Sta=4958.8,5060.9
XS Rating Curve= 0 ,0
Exp/Cntr=0.3,0.1

Type RM Length L Ch R = 1 ,33799   ,477,477,477
BEGIN DESCRIPTION:
UNT094 IN BECR 50.0
END DESCRIPTION:
XS GIS Cut Line= 3
      3776899.59     10559160.21      3776499.61     10559710.19
      3776249.59     10560060.22
#Sta/Elev= 30
  4321.2   350.6  4378.7   346.8  4445.8  336.66  4468.4  331.79  4520.9   323.9
  4529.4  321.34  4550.3  319.11    4606     318  4704.4  320.27  4742.7  321.69
  4786.8  320.49  4887.3   311.9    4929  311.47  4951.8  313.36  4964.5  310.51
    4973  312.13  4979.2   308.2  4984.7  308.12  4987.5  307.62  4990.7  308.12
  5023.4  309.41  5029.5  312.61  5038.1  313.16  5065.1  311.72  5095.6  313.42
  5165.9  311.76  5186.8  314.36  5296.2  321.78  5367.5  329.84  5431.4  333.96
#Mann= 8 ,-1 , 0
  4321.2     .05       0  4445.8     .16       0  4468.4     .12       0
    4606     .16       0  4704.4     .12       0  4984.7     .07       0
  4990.7     .12       0  5095.6     .16       0
Bank Sta=4951.8,5038.1
XS Rating Curve= 0 ,0
Exp/Cntr=0.3,0.1

Type RM Length L Ch R = 1 ,33322   ,524,524,524
BEGIN DESCRIPTION:
UNT094 IN BECR 49.0
END DESCRIPTION:
XS GIS Cut Line= 3
      3776749.62     10559060.18      3776149.61     10559410.19
      3775699.62     10559510.19
#Sta/Elev= 30
  4348.2  342.49  4393.3  339.56  4424.4  334.62  4473.5  329.72  4487.1   330.3
  4559.5  320.48  4590.9  320.52  4618.2  317.47  4705.3  318.16  4751.5  319.18
  4778.6  318.88  4800.1  315.79  4822.4   315.1  4939.5  312.72  4961.8  313.28
  4994.8  308.19  4997.5  307.69  5000.8  308.19  5013.5  312.07  5019.7  311.16
  5029.2  312.91    5094  309.91  5145.3  311.42  5154.2  313.14  5159.4  311.64
  5243.9  310.66  5343.7  316.41  5370.6  318.95  5421.9  328.07  5503.8     334
#Mann= 9 ,-1 , 0
  4348.2     .05       0  4424.4     .16       0  4705.3     .05       0
  4751.5     .16       0  4822.4     .05       0  4939.5     .12       0
  4994.8     .07       0  5000.8     .12       0  5243.9     .16       0
Bank Sta=4961.8,5029.2
XS Rating Curve= 0 ,0
Exp/Cntr=0.3,0.1

Type RM Length L Ch R = 1 ,32798   ,206,206,206
BEGIN DESCRIPTION:
UNT094 IN BECR 48.0
END DESCRIPTION:
XS GIS Cut Line= 3
      3776599.61     10558060.19      3775799.61     10559160.19
      3775599.64     10559310.16
#Sta/Elev= 30
  3619.7  357.26  3733.5  352.07  3842.3   345.1  3899.1  336.79  3919.9  335.62
  3941.2  330.37  3978.3  326.31  3984.8  324.15  4020.4  320.67  4141.7  313.77
  4313.3   313.2  4549.8  309.35  4635.6  309.05  4650.2  310.29  4707.8  309.01
  4721.3  310.46  4754.3  308.98    4757  308.48  4760.3  308.98  4907.6  311.35
  4930.4  310.31  4972.5  311.81    4983  311.12  4987.1  309.21  5016.3  310.73
  5072.6  309.77  5101.7  313.95  5137.1  322.54  5187.1  328.06  5229.8  330.32
#Mann= 6 ,-1 , 0
  3619.7     .05       0  3733.5     .16       0  4020.4     .16       0
  4754.3     .07       0  4760.3     .16       0  5187.1     .16       0
#XS Ineff= 2 , 0
         4667.73  322.53
Permanent Ineff=
       F       F
Bank Sta=4721.3,4907.6
XS Rating Curve= 0 ,0
Exp/Cntr=0.3,0.1

Type RM Length L Ch R = 1 ,32592   ,918,918,918
BEGIN DESCRIPTION:
UNT094 IN BECR 47.0
END DESCRIPTION:
XS GIS Cut Line= 2
      3776257.64     10558084.96      3775233.96     10559681.21
#Sta/Elev= 30
  3888.7  348.06  3949.1  346.27    4043   338.9  4173.1   320.2  4224.7  315.58
  4339.6  310.92  4693.8  308.73  4738.4  310.17  4787.7  308.62  4796.9  310.05
  4809.6  308.56    4976  310.92  4999.5  307.95  5002.7  308.45    5009  310.05
  5020.9  310.59  5120.7  309.05  5193.4  316.06  5201.7  318.86  5244.9   325.4
  5281.3  327.32  5338.8  327.94  5344.7  326.27  5432.6   325.6  5484.1   326.7
  5490.1   325.7    5583  331.98  5589.9  332.15    5665  337.46    5785  342.84
#Mann= 7 ,-1 , 0
  3888.7     .16       0  4173.1   .0316       0  5002.7     .05       0
    5009    .126       0  5484.1     .16       0    5583      .1       0
  5589.9     .16       0
#XS Ineff= 2 , 0
         4772.73   321.9
Permanent Ineff=
       F       F
Bank Sta=4976,5020.9
XS Rating Curve= 0 ,0
Exp/Cntr=0.3,0.1

Type RM Length L Ch R = 1 ,31674   ,617,617,617
BEGIN DESCRIPTION:
UNT094 IN BECR 46.0
END DESCRIPTION:
XS GIS Cut Line= 3
       3775499.6     10557910.21      3774849.61     10559060.19
       3775099.6     10559810.16
#Sta/Elev= 30
  3639.5  346.64    3685  344.52  3690.7  345.88  3706.6  343.82  3755.7  343.07
  3765.8  340.89  3793.2   340.9  3895.7  329.99  3933.3  321.55    3939  319.52
  3984.1  313.19  4240.8  309.14  4548.3  308.18  4569.9   309.7  4592.9  307.47
  4799.6  307.46    4971  309.35  5002.6  307.99  5034.2  309.55  5076.4  307.64
  5171.3  309.65  5192.4  307.53  5252.6  307.29  5255.4  306.79  5258.6  307.29
  5276.7  309.62  5413.7  314.36  5540.2  327.64    5614  336.54    5751  348.72
#Mann= 5 ,-1 , 0
  3639.5     .16       0  3933.3     .16       0  5252.6     .07       0
  5258.6     .16       0  5540.2     .16       0
#XS Ineff= 2 , 0
                         5284.09          317.71
Permanent Ineff=
       F       F
Bank Sta=5171.3,5276.7
XS Rating Curve= 0 ,0
Exp/Cntr=0.3,0.1

Type RM Length L Ch R = 1 ,31057   ,336,336,336
BEGIN DESCRIPTION:
UNT094 IN BECR 45.0
END DESCRIPTION:
XS GIS Cut Line= 3
      3775432.96     10557859.31      3774643.04     10558918.32
      3774330.55      10560289.8
#Sta/Elev= 30
  3168.6  348.95  3314.8  345.71    3371   341.7    3394   338.3  3421.1  330.39
    3444  327.48  3500.3  318.31  3585.8  311.65  3643.8  312.42  3793.5  307.66
  4527.6  306.53  4572.8  305.83  4575.5  305.33  4578.8  305.83  4661.8  306.98
  4881.4  308.59  4963.5  306.94  4973.2  310.34  4978.4  306.85    4984  308.46
  4994.2   306.7  5127.6  306.93  5219.9  309.66  5281.4  314.11  5332.7  313.77
    5343  316.18  5486.5  325.04  5671.2  341.47  5769.4  348.06  5896.4  351.04
#Mann= 7 ,-1 , 0
  3168.6     .16       0    3444     .07       0  3585.8     .16       0
  4572.8    .035       0  4578.8     .16       0  5486.5      .1       0
  5769.4     .05       0
#XS Ineff= 2 , 0
                         4811.93           322.6
Permanent Ineff=
       F       F
Bank Sta=4527.6,4661.8
XS Rating Curve= 0 ,0
Exp/Cntr=0.3,0.1

Type RM Length L Ch R = 1 ,30721   ,1241,1241,1241
BEGIN DESCRIPTION:
UNT094 IN BECR 44.0
END DESCRIPTION:
XS GIS Cut Line= 3
      3774851.36     10557642.32      3774174.29     10559473.88
      3774130.89     10560194.37
#Sta/Elev= 30
  3170.7  356.56  3384.5  346.79    3445   343.4  3520.3  336.25  3561.3   327.8
  3616.2  319.21  3637.5   313.2  3677.7  307.74  3701.5  308.08  4001.5  305.31
  4519.4  305.28  4522.2  304.78  4525.4  305.28  4703.7  305.46  4719.2  306.75
    4725  305.32    4891  308.06  4896.3  306.52  4951.8  306.01  5068.1  305.86
  5098.6  307.97  5122.9  306.87    5270   311.8  5390.2  320.39  5415.9  321.98
    5453  326.87  5550.5  334.67  5616.3  338.97  5703.2  341.74  5845.2  345.27
#Mann= 8 ,-1 , 0
  3170.7     .16       0  3384.5     .12       0  3520.3     .16       0
  4519.4    .033       0  4525.4     .16       0  5390.2     .16       0
  5415.9      .1       0  5703.2     .16       0
#XS Ineff= 2 , 0
                         4892.05           316.6
Permanent Ineff=
       F       F
Bank Sta=3701.5,4891
XS Rating Curve= 0 ,0
Exp/Cntr=0.3,0.1

Type RM Length L Ch R = 1 ,29480   ,571,571,571
BEGIN DESCRIPTION:
UNT094 IN BECR 43.0
END DESCRIPTION:
XS GIS Cut Line= 4
      3774356.59     10557477.34      3773879.15     10558171.79
      3773801.03     10558935.68       3773931.1     10559976.27
#Sta/Elev= 30
  3935.2  351.09  4216.4  342.09  4315.1  334.39  4452.5  315.56  4473.5  311.16
    4554  304.71  4646.7  306.06  4748.2  304.15  4827.1  304.73  4883.9  303.91
  4886.7  303.41  4889.9  303.91  5108.1  305.43  5178.4  304.89  5208.6  306.47
    5289  314.21  5339.3  317.01  5459.9  329.68  5507.9  332.39  5600.7  331.62
  5671.3  333.78  5862.8   325.5  5892.6   320.1  6053.8  320.11  6139.5  322.84
  6366.7  334.96  6527.9  337.17  6542.6  338.89  6588.4  339.54  6594.5  339.68
#Mann= 5 ,-1 , 0
  3935.2     .16       0  4216.4     .16       0  4883.9     .07       0
  4889.9     .16       0  6588.4     .05       0
#XS Ineff= 2 , 0
                         5134.66          318.32
Permanent Ineff=
       F       F
Bank Sta=4827.1,5108.1
XS Rating Curve= 0 ,0
Exp/Cntr=0.3,0.1

Type RM Length L Ch R = 1 ,28909   ,634,634,634
BEGIN DESCRIPTION:
UNT094 IN BECR 42.0
END DESCRIPTION:
XS GIS Cut Line= 3
      3773245.48     10558024.26      3773462.48     10558805.48
      3773870.47     10559951.32
#Sta/Elev= 30
  4472.2  331.51    4579  332.34  4618.4  330.19  4644.4  326.68  4665.2  321.31
  4675.5  316.71  4685.9  316.07  4697.3  312.15  4737.8  304.38  4945.4  304.08
  4994.3  303.14    4997  302.64  5000.3  303.14  5049.2  304.78  5070.9  303.47
  5286.2  303.94  5763.3   307.4  5850.5   310.4  6004.7  312.43  6030.2  314.16
  6035.5  316.99    6061  316.35  6066.3  318.44  6091.8  318.94  6097.2  321.04
  6105.3  321.65    6179  321.51  6182.3  322.77  6287.9  327.38  6499.3  337.44
#Mann= 6 ,-1 , 0
  4472.2     .16       0  4994.3     .07       0  5000.3     .12       0
  6091.8     .16       0  6182.3      .1       0  6287.9     .05       0
#XS Ineff= 2 , 0
                          5235.8          314.97
Permanent Ineff=
       F       F
Bank Sta=4945.4,5049.2
XS Rating Curve= 0 ,0
Exp/Cntr=0.3,0.1

Type RM Length L Ch R = 1 ,28275   ,560,560,560
BEGIN DESCRIPTION:
UNT094 IN BECR 41.0
END DESCRIPTION:
XS GIS Cut Line= 3
      3773149.61     10558210.18      3772899.61     10558710.19
      3772749.61     10559360.18
#Sta/Elev= 30
  4423.1  330.18  4431.5  330.56  4467.8  326.29  4476.2  323.62  4512.5  317.44
  4520.9  314.52  4534.9  311.84  4557.3  308.86  4571.2  308.28  4593.6  304.11
  4691.4  302.81  4825.6  302.62    4848  304.23  4884.3   302.8  4959.8  303.19
  5020.2  302.05  5022.9  301.55  5026.2  302.05  5187.4  302.61  5213.5   302.8
    5290  304.67  5351.6  308.39  5401.2   315.4  5406.3  314.82  5443.9  320.06
  5505.5  325.98  5577.4  335.77  5608.2   337.5  5625.3     341  5649.2  342.92
#Mann= 4 ,-1 , 0
  4423.1     .12       0  5020.2     .07       0  5026.2     .12       0
  5213.5     .16       0
Bank Sta=4959.8,5187.4
XS Rating Curve= 0 ,0
Exp/Cntr=0.3,0.1

Type RM Length L Ch R = 1 ,27715   ,537,537,537
BEGIN DESCRIPTION:
UNT094 IN BECR 40.0
END DESCRIPTION:
XS GIS Cut Line= 3
      3773049.58     10558160.21      3772449.61     10558610.19
      3771749.66     10558760.18
#Sta/Elev= 30
  4211.5  328.84  4283.3  325.29  4289.6  322.93  4354.2   315.3  4368.8  315.77
    4375  314.11  4454.2  308.56  4589.6  301.76  4611.5  301.07    4625  302.72
  4954.2  300.79  4981.1  301.67  5027.5  300.37  5030.2  299.87  5033.5  300.37
  5035.6   301.5  5224.9  301.68  5287.1  303.29  5350.1   307.7  5410.6  314.56
  5421.7  318.13  5452.4  322.66    5460  325.42  5489.1   331.1  5523.9  339.59
  5544.4  343.01  5558.9  343.65  5575.1  347.14  5646.7  352.94  5677.3  353.16
#Mann= 6 ,-1 , 0
  4211.5     .12       0  5027.5     .07       0  5033.5     .12       0
  5224.9     .16       0  5287.1     .12       0  5489.1     .16       0
Bank Sta=4981.1,5035.6
XS Rating Curve= 0 ,0
Exp/Cntr=0.3,0.1

Type RM Length L Ch R = 1 ,27178   ,538,538,538
BEGIN DESCRIPTION:
UNT094 IN BECR 39.0
END DESCRIPTION:
XS GIS Cut Line= 3
      3772849.65     10557810.16      3772099.61     10558310.19
      3771699.65     10558360.18
#Sta/Elev= 30
  4123.9  327.76  4196.1  325.59  4239.6   322.5  4383.8  306.65  4389.9  307.13
    4471  300.41  4888.6  300.09  4894.6   299.3  4924.7  300.06  4945.7  299.19
  4981.8  300.98  4989.3  300.62  4993.8  298.58  4996.5  298.08  4999.8  298.58
  5017.8  300.02  5055.6  299.44  5095.1  300.85  5136.2  303.45  5156.3  306.63
  5176.5   310.4  5206.7  318.85  5216.8  320.32  5224.4  323.06    5237  325.01
    5247  328.09  5317.6  341.34  5337.7   342.8    5368  347.62  5428.4  351.17
#Mann= 4 ,-1 , 0
  4123.9     .12       0  4993.8     .07       0  4999.8     .12       0
  5095.1     .16       0
Bank Sta=4981.8,5017.8
XS Rating Curve= 0 ,0
Exp/Cntr=0.3,0.1

Type RM Length L Ch R = 1 ,26640   ,507,507,507
BEGIN DESCRIPTION:
UNT094 IN BECR 38.0
END DESCRIPTION:
XS GIS Cut Line= 3
      3772749.65     10557760.19      3771999.61     10557810.19
       3771699.6      10558160.2
#Sta/Elev= 30
  4263.5  324.48  4293.6  322.34  4343.7  320.64  4393.8  317.21  4413.9  313.73
    4484  304.99  4524.1  301.37  4564.2  298.95  4654.4  298.21    4925  298.72
  4945.1  298.28  4955.1  297.16  4985.1  298.32  4992.2  295.86  4994.9  295.36
  4998.2  295.86  5015.2  298.01  5028.9  298.17  5133.7  304.77  5185.9  307.88
  5206.7  311.31  5256.1  315.87  5291.8  321.38  5298.9  324.02  5313.2  326.48
  5334.1   328.1  5341.7  330.38  5376.9  334.24    5384  336.21  5476.2  344.09
#Mann= 4 ,-1 , 0
  4263.5     .12       0  4992.2     .07       0  4998.2     .12       0
  5133.7     .16       0
Bank Sta=4985.1,5015.2
XS Rating Curve= 0 ,0
Exp/Cntr=0.3,0.1

Type RM Length L Ch R = 1 ,26133   ,562,562,562
BEGIN DESCRIPTION:
UNT094 IN BECR 37.0
END DESCRIPTION:
XS GIS Cut Line= 3
      3773249.63     10556060.16      3771849.61     10557360.19
      3771499.65     10557560.17
#Sta/Elev= 30
    3066  361.62  3401.7  346.79  3426.9  346.15  3526.1  337.94  3547.1  333.78
  3568.6   331.6  3575.4  329.34  3596.9  327.25    3849   312.8  3936.5  304.65
  4297.1  303.17  4580.5  297.85  4587.3  298.89  4693.4  296.65  4856.1  296.66
  4874.6  294.08  4877.3  293.58  4880.6  294.08  4884.4  296.01  4979.4   296.5
  4999.6  294.25    5006  296.48  5030.5  298.16  5086.7  304.28  5129.9  306.67
  5183.1   320.1  5226.3   323.7  5269.5  329.75  5328.5  334.43  5379.6  334.67
#Mann= 6 ,-1 , 0
    3066     .05       0  3401.7     .16       0    3849     .12       0
  4874.6     .07       0  4880.6     .12       0  5030.5     .16       0
Bank Sta=4856.1,4884.4
XS Rating Curve= 0 ,0
Exp/Cntr=0.3,0.1

Type RM Length L Ch R = 1 ,25571   ,516,516,516
BEGIN DESCRIPTION:
UNT094 IN BECR 36.0
END DESCRIPTION:
XS GIS Cut Line= 3
      3772349.64     10556260.15      3771849.61     10556860.19
      3771549.64     10557210.15
#Sta/Elev= 30
  4228.5  329.46  4313.8  325.94  4320.3  323.58  4427.1  314.07  4477.8  305.01
    4541  298.73  4619.1  296.85  4704.3  297.91  4945.1  296.92  4959.5  296.37
  4973.8  293.52  4999.4  293.39  5002.2  292.89  5005.4  293.39  5037.6  298.05
  5066.1  300.35  5073.8  303.08    5088  304.33  5094.6  303.43  5108.9  305.39
  5123.2  305.92  5129.8  304.58  5186.8  306.77  5201.1  308.72  5224.5   308.4
  5264.8  307.92  5293.3  309.63  5350.4  313.63  5428.3  321.89  5470.5  323.62
#Mann= 5 ,-1 , 0
  4228.5     .16       0  4477.8     .12       0  4999.4     .07       0
  5005.4     .12       0  5224.5     .16       0
Bank Sta=4945.1,5037.6
XS Rating Curve= 0 ,0
Exp/Cntr=0.3,0.1

Type RM Length L Ch R = 1 ,25055   ,555,555,555
BEGIN DESCRIPTION:
UNT094 IN BECR 35.0
END DESCRIPTION:
XS GIS Cut Line= 3
      3771949.58     10556110.22      3771649.61     10556410.19
      3771149.62     10556960.17
#Sta/Elev= 30
  4584.6  321.54    4627  319.88  4669.4  316.48    4726  307.98    4778  303.06
    4825  299.18  4895.7  296.88  4938.1  294.11  4980.5  295.72  5002.3  293.72
    5005  293.22  5008.3  293.72  5015.9     294  5022.7  295.71  5093.6   294.6
  5228.1  295.13  5249.7  294.24  5341.6  294.71  5464.3  297.09  5525.4  303.02
    5547   303.5    5568  306.83  5582.2  307.16  5589.6  309.47  5610.6  312.28
  5631.5  313.36  5681.5  319.85  5695.7  320.38  5730.8  324.89  5752.1  326.43
#Mann= 5 ,-1 , 0
  4584.6     .16       0    4778     .12       0  5002.3     .07       0
  5008.3     .12       0  5464.3     .16       0
Bank Sta=4980.5,5022.7
XS Rating Curve= 0 ,0
Exp/Cntr=0.3,0.1

Type RM Length L Ch R = 1 ,24500   ,478,478,478
BEGIN DESCRIPTION:
UNT094 IN BECR 34.0
END DESCRIPTION:
XS GIS Cut Line= 3
       3771599.6     10555660.21      3771399.61     10556010.19
      3770899.61     10556510.19
#Sta/Elev= 30
  4581.9  322.96  4623.6  323.23  4676.2  319.76  4713.6  313.54  4720.1  311.38
  4735.2  309.97  4743.1  307.11  4778.1  304.09  4794.2  302.56  4800.7  299.76
  4823.7   296.3  4853.3  293.92  4977.1  294.14  4982.1  292.25  4999.1   292.1
  5041.6  293.82  5095.5  292.98  5126.4  293.67  5241.8   292.8  5264.8  291.88
  5267.6  291.38  5270.8  291.88  5279.9  292.13  5324.4  292.35  5366.8  294.76
  5387.2  296.05  5437.5   302.2  5573.9  314.74  5647.4  323.12  5692.1   327.2
#Mann= 11 ,-1 , 0
  4581.9     .05       0  4623.6     .16       0  4778.1     .12       0
  5095.5     .16       0  5241.8     .05       0  5264.8     .07       0
  5270.8     .05       0  5279.9     .12       0  5387.2     .16       0
  5573.9     .12       0  5647.4     .16       0
Bank Sta=5126.4,5366.8
XS Rating Curve= 0 ,0
Exp/Cntr=0.3,0.1

Type RM Length L Ch R = 1 ,24022   ,589,589,589
BEGIN DESCRIPTION:
UNT094 IN BECR 33.0
END DESCRIPTION:
XS GIS Cut Line= 3
      3771599.59      10555460.2      3771249.61     10555660.19
      3770799.59      10556010.2
#Sta/Elev= 30
  4570.3  321.61  4658.8  323.39  4673.9  324.55  4740.7  324.42  4804.2  322.78
  4857.5  317.75  4879.1  314.23  4892.8  313.19  4900.7  310.56  4922.3  307.15
  4943.9  305.13  4950.4  302.82  4965.5  300.18  4970.5  297.86  4976.6  297.86
  4980.6  296.86  4992.1  290.55  4994.9  290.05  4998.1  290.55  5021.9  292.84
  5024.1  293.09  5087.4   292.7  5138.1  294.33  5343.5  297.52  5407.7  307.88
  5422.2   309.2  5451.2  314.54  5480.1  317.18  5492.8  319.55  5543.5  323.43
#Mann= 5 ,-1 , 0
  4570.3     .05       0  4740.7     .16       0  4992.1     .07       0
  4998.1     .16       0  5021.9     .05       0
Bank Sta=4976.6,5024.1
XS Rating Curve= 0 ,0
Exp/Cntr=0.3,0.1

Type RM Length L Ch R = 1 ,23433   ,504,504,504
BEGIN DESCRIPTION:
UNT094 IN BECR 32.0
END DESCRIPTION:
XS GIS Cut Line= 3
       3771699.6      10554760.2      3770899.61     10555210.19
      3770349.57     10555210.19
#Sta/Elev= 30
  4101.3  330.16  4174.3  323.67  4181.6  321.61  4239.3  319.73  4292.8  321.07
  4352.1  316.26  4357.8  317.46  4401.2   314.2  4476.4  303.85  4521.7  301.73
  4601.7  299.47  4703.3  299.17  4732.3  295.17  4740.9  298.49  4755.3   298.8
  4842.4   296.4  4865.2  293.95    4871   295.9  4886.9  295.97  4930.2  293.68
  4983.8  294.47  4989.5  294.17  4993.2  290.17    4996  289.67  4999.2  290.17
  5016.3  293.12  5059.2  294.93  5329.2  295.59  5469.2  312.23  5569.2  318.63
#Mann= 7 ,-1 , 0
  4101.3     .16       0  4521.7     .12       0  4601.7     .05       0
  4842.4     .16       0  4983.8     .05       0  4993.2     .03       0
  4999.2     .05       0
Bank Sta=4983.8,5059.2
XS Rating Curve= 0 ,0
Exp/Cntr=0.3,0.1

Type RM Length L Ch R = 1 ,22929   ,546,546,546
BEGIN DESCRIPTION:
UNT094 IN BECR 31.0
END DESCRIPTION:
XS GIS Cut Line= 3
      3771699.57     10554710.19      3770899.61     10554760.19
      3770499.64      10554660.2
#Sta/Elev= 30
  4162.1  330.48  4182.1  326.49  4202.1  324.38  4292.3  318.41  4312.3  315.11
    4424  304.21  4532.8  294.83  4612.9  293.25    4688  293.81  4724.3  293.37
  4784.3  293.11  4883.4  292.56  4927.6  293.47  4953.6  293.85  4981.7  291.61
  4986.8  288.49  5001.8   288.1  5004.6   287.6  5007.8   288.1  5015.2  292.24
    5028  292.97  5064.1  294.53  5105.3  299.74  5138.8  301.51  5144.3  304.09
  5146.6  305.17  5159.5  304.39  5200.7  312.67    5345   324.5  5375.9  325.46
#Mann= 10 ,-1 , 0
  4162.1     .16       0    4424     .12       0    4688     .07       0
  4724.3     .05       0  4784.3     .07       0  4883.4     .05       0
  4927.6     .12       0  5001.8     .07       0  5007.8     .12       0
  5144.3     .05       0
Bank Sta=4953.6,5028
XS Rating Curve= 0 ,0
Exp/Cntr=0.3,0.1

Type RM Length L Ch R = 1 ,22383   ,204,204,204
BEGIN DESCRIPTION:
UNT094 IN BECR 30.0
END DESCRIPTION:
XS GIS Cut Line= 4
      3771870.07      10553853.9      3771151.32     10554150.78
      3770812.78     10554400.78      3770303.48     10554619.05
#Sta/Elev= 30
  4021.3  358.02  4088.5  354.05    4109  352.23  4204.8  343.78  4344.1  335.66
  4422.2  328.66  4441.1  322.28  4523.6  315.57  4547.5  306.51  4579.2  305.46
  4639.6   300.3  4768.3  292.16    4978  292.63    4997  288.61  4999.7  288.11
    5003  288.61  5007.3  292.36  5092.9  299.21  5107.5  296.87  5113.7  300.69
  5122.1  298.34  5128.4   304.1    5143  300.25  5149.2  306.29  5210.9  313.15
  5411.2  320.53  5434.7  322.63  5440.8  327.08  5458.3  323.04  5773.9  331.15
#Mann= 11 ,-1 , 0
  4021.3     .16       0  4088.5     .05       0    4109     .16       0
  4204.8     .05       0  4344.1     .16       0  4422.2     .05       0
  4579.2     .16       0  4639.6     .12       0    4997     .07       0
    5003     .12       0  5210.9     .05       0
Bank Sta=4978,5007.3
XS Rating Curve= 0 ,0
Exp/Cntr=0.3,0.1

Type RM Length L Ch R = 1 ,22179   ,813,813,813
BEGIN DESCRIPTION:
UNT094 IN BECR 29.0
END DESCRIPTION:
XS GIS Cut Line= 4
       3771885.7     10553562.23      3771526.32     10553874.74
      3770849.24     10554135.15       3770396.1     10554327.87
#Sta/Elev= 30
  3952.6  375.11  4033.4  368.09  4288.9  337.07  4366.7  331.53  4388.8  332.51
  4446.8  331.81    4560  323.42  4629.7   318.5  4671.8  312.14  4683.8  307.98
  4763.6  295.44  4818.2  293.47  4878.2  294.56  4939.6  290.82  4982.2   292.2
  4987.5  291.17  4993.2  286.85  5000.9  286.79  5003.6  286.29  5006.9  286.79
  5025.3  292.67    5036  293.28  5126.8  298.25  5180.5  304.45  5233.2  306.83
    5393  319.27    5415  323.06  5462.3  324.56  5485.9  327.48  5646.7  330.89
#Mann= 6 ,-1 , 0
  3952.6     .16       0  4388.8     .05       0    4560     .16       0
  4683.8     .05       0  5000.9     .04       0  5006.9     .05       0
Bank Sta=4982.2,5036
XS Rating Curve= 0 ,0
Exp/Cntr=0.3,0.1

Type RM Length L Ch R = 1 ,21366   ,702,702,702
BEGIN DESCRIPTION:
UNT094 IN BECR 28.0
END DESCRIPTION:
XS GIS Cut Line= 3
      3771281.53     10553218.49      3770651.32     10553447.65
      3770401.31     10553932.06
#Sta/Elev= 30
  4440.7  327.25    4546  319.73  4551.3  320.96  4599.7  320.76    4663  320.04
  4693.6  318.11  4785.4  310.23  4801.4  307.18  4810.6  304.68  4942.9  288.38
  4983.6  291.33  4988.9  290.44  4996.1   284.6  5003.7  284.38  5006.5  283.88
  5009.7  284.38  5019.5  290.74  5038.6  288.58  5239.2  289.79  5271.7  291.68
  5283.6  294.64  5316.6  297.59  5338.8  297.58  5418.5  308.31  5440.5   311.6
  5471.7  313.85  5485.5  317.29  5543.8   323.2  5626.8  323.91  5656.4  321.55
#Mann= 6 ,-1 , 0
  4440.7     .05       0  4599.7     .16       0  4801.4     .12       0
  5003.7     .07       0  5009.7     .12       0  5418.5     .05       0
Bank Sta=4983.6,5019.5
XS Rating Curve= 0 ,0
Exp/Cntr=0.3,0.1

Type RM Length L Ch R = 1 ,20664   ,558,558,558
BEGIN DESCRIPTION:
UNT094 IN BECR 27.0
END DESCRIPTION:
XS GIS Cut Line= 3
       3770899.6     10552560.19      3770399.61     10552910.19
      3769899.64     10553110.18
#Sta/Elev= 30
  4425.5  322.19  4462.1  320.93  4504.4  317.14  4519.2  313.73  4569.8   305.9
  4596.8  299.44  4656.1  294.23  4719.7  292.02  4805.2  288.69  4913.8  287.91
  4977.8  289.34  4986.6  287.09  4989.7  283.88  4992.4  283.38  4995.7  283.88
  5007.5  286.32  5013.6  289.38  5074.9   287.3  5111.2   288.2  5134.1  287.03
  5158.3  288.19  5182.6  286.62    5224  287.28  5319.9  294.91  5326.6  296.83
  5422.2  307.26  5451.8  311.91  5520.5  317.74  5529.9  320.85  5574.3  324.08
#Mann= 5 ,-1 , 0
  4425.5     .16       0  4719.7     .12       0  4989.7     .07       0
  4995.7     .12       0    5224     .16       0
Bank Sta=4977.8,5013.6
XS Rating Curve= 0 ,0
Exp/Cntr=0.3,0.1

Type RM Length L Ch R = 1 ,20106   ,638,638,638
BEGIN DESCRIPTION:
UNT094 IN BECR 26.0
END DESCRIPTION:
XS GIS Cut Line= 3
      3770699.58     10552360.19      3770249.61     10552460.19
       3769499.6     10552560.19
#Sta/Elev= 30
  4493.6  316.65  4503.8  314.77  4512.8  310.89  4565.8  302.63  4616.5  293.46
  4708.7  285.73  4974.7  287.58  4984.8  286.06  4991.1  283.39  4996.2   286.4
    5002  281.69  5004.7  281.19    5008  281.69  5015.1  281.81  5035.3  287.57
  5045.3  288.18  5147.5  286.05  5220.6  288.92  5277.4  298.64  5307.6  308.86
  5327.8  312.05  5366.9  312.64    5372  315.92  5375.5  315.76  5398.4  318.43
  5408.5  321.97  5438.8  327.93  5518.2  336.15  5669.6  347.79  5711.2  352.55
#Mann= 5 ,-1 , 0
  4493.6     .16       0  4565.8     .12       0    5002     .07       0
    5008     .12       0  5375.5     .16       0
Bank Sta=4974.7,5045.3
XS Rating Curve= 0 ,0
Exp/Cntr=0.3,0.1

Type RM Length L Ch R = 1 ,19468   ,556,556,556
BEGIN DESCRIPTION:
UNT094 IN BECR 25.0
END DESCRIPTION:
XS GIS Cut Line= 3
      3771156.49     10551827.87      3770199.61     10552010.19
      3769399.63     10552410.18
#Sta/Elev= 30
  4025.3  332.02  4222.7  323.24  4332.1  306.64  4337.7  303.88  4378.4  297.36
  4389.3  301.13  4422.9  304.96  4441.5  308.62  4493.7  309.08  4545.8  303.02
    4598  292.92  4673.6   287.4  4958.7  283.96  4973.3  285.41  4993.8  280.97
  4996.6  280.47  4999.8  280.97  5007.8  285.05  5021.8  286.29    5263  285.35
  5365.5  293.52    5455  297.36    5469  296.19  5639.5   312.4  5737.3  329.76
  5751.3  337.73  5863.1  350.91  5879.8  354.51  5885.4  353.62  5893.8  355.99
#Mann= 5 ,-1 , 0
  4025.3     .16       0  4422.9     .12       0  4993.8     .07       0
  4999.8     .12       0    5263     .16       0
Bank Sta=4973.3,5021.8
XS Rating Curve= 0 ,0
Exp/Cntr=0.3,0.1

Type RM Length L Ch R = 1 ,18912   ,594,594,594
BEGIN DESCRIPTION:
UNT094 IN BECR 24.0
END DESCRIPTION:
XS GIS Cut Line= 3
      3770749.65     10551260.17      3769953.41     10551588.28
      3769255.48     10551937.24
#Sta/Elev= 30
  4165.3  322.84    4180  322.67  4334.5  304.76  4403.3  299.71    4465  298.65
  4515.1  292.83  4608.8  284.63  4630.4  284.07  4954.9  285.05  4976.5  283.81
  4989.4  280.29  4992.2  279.79  4995.4  280.29    5009  284.62  5097.8  284.81
  5155.4  287.81  5195.7  289.06    5232  292.71  5262.7  293.02  5343.8  304.52
  5441.6   314.6  5447.2  313.62    5464  315.77    5478  314.88  5508.7  317.15
  5536.7  316.49  5553.4  318.49  5581.4  318.63  5723.9  332.44  5806.8  336.89
#Mann= 5 ,-1 , 0
  4165.3     .16       0  4515.1     .12       0  4989.4     .07       0
  4995.4     .12       0  5155.4     .16       0
Bank Sta=4954.9,5009
XS Rating Curve= 0 ,0
Exp/Cntr=0.3,0.1

Type RM Length L Ch R = 1 ,18318   ,503,503,503
BEGIN DESCRIPTION:
UNT094 IN BECR 23.0
END DESCRIPTION:
XS GIS Cut Line= 3
      3770649.66     10551110.19      3769849.61     10551110.19
      3769499.58     10551510.22
#Sta/Elev= 30
  4237.6  316.89  4287.6  312.29  4407.6  297.48  4457.6  294.46  4577.6  290.47
  4607.6  290.62  4617.6  289.19  4707.6  286.33  4957.6  283.71  4977.6  279.44
  5017.6  280.07  5035.1  284.37    5041  284.37  5044.8  279.72  5070.2   279.1
    5073   278.6  5076.2   279.1  5079.9  281.14  5094.1  283.11  5186.2  284.55
  5257.4  283.86  5377.9  287.18  5434.9  294.34  5449.1  298.74  5455.7  299.33
  5476.6  303.34  5484.2  307.35  5505.1  310.15  5512.7  313.15  5569.2  318.95
#Mann= 5 ,-1 , 0
  4237.6     .16       0  4457.6     .16       0  5070.2     .07       0
  5076.2     .16       0  5455.7     .16       0
Bank Sta=5041,5094.1
XS Rating Curve= 0 ,0
Exp/Cntr=0.3,0.1

Type RM Length L Ch R = 1 ,17815   ,598,598,598
BEGIN DESCRIPTION:
UNT094 IN BECR 22.0
END DESCRIPTION:
XS GIS Cut Line= 3
      3771299.65     10550160.17      3769749.61     10550710.19
      3769049.63     10550660.19
#Sta/Elev= 30
  3361.1  366.24    3413  363.02  3494.7  355.84  3594.6  350.76  3721.9  341.09
  3743.1  339.48  3792.8  329.27  3806.8  328.17  3934.1   299.8  4008.9  293.84
  4121.8  290.33  4645.1   289.8  4754.1  286.68  4942.2  285.19    4974  284.23
  4984.6   282.2  4990.4  278.81  5000.2  277.97  5002.9  277.47  5006.2  277.97
  5015.9   278.1  5035.9  285.24  5218.9  286.76  5286.6  289.81  5366.8  296.43
  5416.9  297.18    5457  301.64  5499.6  304.49  5634.9  320.96  5707.6  327.65
#Mann= 6 ,-1 , 0
  3361.1     .05       0    3413     .16       0  3721.9     .16       0
  5000.2     .07       0  5006.2     .16       0    5457     .16       0
#XS Ineff= 2 , 0
         4827.27   299.8
Permanent Ineff=
       F       F
Bank Sta=4942.2,5035.9
XS Rating Curve= 0 ,0
Exp/Cntr=0.3,0.1

Type RM Length L Ch R = 1 ,17217   ,550,550,550
BEGIN DESCRIPTION:
UNT094 IN BECR 21.0
END DESCRIPTION:
XS GIS Cut Line= 3
      3771099.62     10549510.18      3769549.61     10550210.19
      3769199.57     10550410.21
#Sta/Elev= 30
  3335.6  369.34  3533.1  355.24    3577  349.08  3586.6  344.95  3592.1  347.15
  3609.7  341.14  3615.2  342.89  3620.9  339.13  3646.2  333.86  3653.8   333.4
  3661.5  329.69  3713.2  321.79  3811.2  311.55  3862.9  307.76  3978.5  294.46
  4076.5  287.07  4410.9  281.99  4893.7  282.78  4970.3  284.68  4995.9  277.92
  4998.7  277.42  5001.9  277.92  5014.4  282.48    5050  285.15  5065.9  283.45
  5087.5  284.54  5130.6  289.93  5211.3  298.03  5286.1  309.85  5439.5  319.32
#Mann= 6 ,-1 , 0
  3335.6     .16       0  3646.2     .05       0  3811.2     .16       0
  4995.9     .07       0  5001.9     .16       0  5130.6     .16       0
#XS Ineff= 2 , 0
         4488.64  305.06
Permanent Ineff=
       F       F
Bank Sta=4970.3,5050
XS Rating Curve= 0 ,0
Exp/Cntr=0.3,0.1

Type RM Length L Ch R = 1 ,16667   ,558,558,558
BEGIN DESCRIPTION:
UNT094 IN BECR 20.0
END DESCRIPTION:
XS GIS Cut Line= 3
      3771099.57      10549410.2      3769549.61     10549810.19
       3768799.6     10550360.19
#Sta/Elev= 30
  3434.4  368.01  3497.9  362.88  3533.4  356.39  3589.3  354.77  3736.2  329.33
  3812.9  317.75  4002.4  298.87  4188.3  285.76  4580.7  281.74  4615.9  278.59
  4632.4  281.33  4673.7  278.85  4704.7  281.23  4838.9  280.38  4962.8  283.39
  5009.2   277.5    5012     277  5015.2   277.5  5024.8  282.26  5157.5  283.08
  5320.4   293.3  5485.5  297.21  5550.3   297.3    5751  312.74  5757.2  315.34
  5768.7  314.31  5886.8  319.18    5893  321.98  5931.5  323.78  5965.2  325.53
#Mann= 8 ,-1 , 0
  3434.4     .16       0  3736.2     .05       0  4002.4     .16       0
  5009.2     .07       0  5015.2     .16       0  5485.5     .16       0
  5768.7      .1       0  5931.5     .16       0
#XS Ineff= 2 , 0
         4632.95  292.14
Permanent Ineff=
       F       F
Bank Sta=4962.8,5024.8
XS Rating Curve= 0 ,0
Exp/Cntr=0.3,0.1

Type RM Length L Ch R = 1 ,16109   ,597,597,597
BEGIN DESCRIPTION:
UNT094 IN BECR 19.0
END DESCRIPTION:
XS GIS Cut Line= 3
      3770349.58     10548560.22      3769549.61     10549310.19
      3768749.62     10550110.18
#Sta/Elev= 30
  3919.9   375.8  4082.7  357.02  4181.4  335.42  4188.7  330.15  4209.8  325.15
  4217.1  328.62  4317.2  320.75  4351.4  313.57  4429.1  310.68  4436.4  313.09
  4443.2  309.24  4457.4  309.51  4464.7  310.97  4471.6  306.73  4485.7   304.6
  4549.7  298.71  4556.6  295.27  4634.2   283.7  4676.7   280.6  4726.5  278.26
  4966.9  280.49  4999.5  277.01  5002.3  276.51  5005.5  277.01  5030.6   280.7
  5652.8  280.17  5879.1  289.66    5964  296.71  6034.7  302.67  6147.8  318.96
#Mann= 6 ,-1 , 0
  3919.9     .16       0  4317.2     .05       0  4457.4     .16       0
  4999.5     .07       0  5005.5     .16       0    5964      .1       0
#XS Ineff= 2 , 0
                         5286.36           297.4
Permanent Ineff=
       F       F
Bank Sta=4966.9,5030.6
XS Rating Curve= 0 ,0
Exp/Cntr=0.3,0.1

Type RM Length L Ch R = 1 ,15512   ,616,616,616
BEGIN DESCRIPTION:
UNT094 IN BECR 18.0
END DESCRIPTION:
XS GIS Cut Line= 3
      3770049.62     10548060.18      3769249.61     10548860.19
      3768649.59      10549110.2
#Sta/Elev= 30
  3858.9  373.52  3901.3  366.65  3914.5  361.89  3986.2  346.74    4071  346.34
  4099.3  350.12  4155.9  330.59  4238.8  321.28  4311.5  316.86  4452.9  302.37
  4608.4  290.94  4735.7  278.68  4792.3  276.75  4947.9  279.11  4976.1  279.13
    4993  277.01  5034.2  279.58  5152.8  276.74  5211.8  277.51  5256.5  276.56
  5259.2  276.06  5262.5  276.56  5282.8  277.63  5294.2  280.37  5389.5  290.34
  5401.9   293.2  5418.7  293.56    5448  299.37  5495.7  303.95  5640.3  312.31
#Mann= 6 ,-1 , 0
  3858.9     .05       0  3914.5     .16       0  4238.8     .05       0
  4311.5     .16       0  5256.5     .07       0  5262.5     .16       0
Bank Sta=5211.8,5294.2
XS Rating Curve= 0 ,0
Exp/Cntr=0.3,0.1

Type RM Length L Ch R = 1 ,14896   ,1164,1164,1164
BEGIN DESCRIPTION:
UNT094 IN BECR 17.0
END DESCRIPTION:
XS GIS Cut Line= 3
      3769799.64     10547910.17      3768999.61     10548460.19
      3768299.57     10548460.19
#Sta/Elev= 30
  4036.8  343.27  4109.7  335.83  4166.7  326.63  4172.8  327.37  4255.8  316.71
  4331.1  308.79  4339.9  306.28    4346  307.27  4360.9  304.26  4442.1  299.95
  4468.5  296.32  4546.5  291.53    4570  291.77  4626.8  283.91  4740.7  276.06
    4827  276.66  4849.9   274.6  4877.8  276.54  4922.4  274.55  4985.3  277.87
  5001.6  273.29  5004.4  272.79  5007.6  273.29  5047.7   277.4  5177.7  277.71
  5327.7  281.49  5417.7  286.07  5457.7  290.77  5487.7  296.75  5707.7  314.56
#Mann= 7 ,-1 , 0
  4036.8     .16       0  4255.8     .05       0  4442.1     .12       0
  4546.5     .16       0  5001.6     .07       0  5007.6     .16       0
  5457.7     .16       0
Bank Sta=4985.3,5047.7
XS Rating Curve= 0 ,0
Exp/Cntr=0.3,0.1

Type RM Length L Ch R = 1 ,13732   ,730,730,730
BEGIN DESCRIPTION:
UNT094 IN BECR 16.0
END DESCRIPTION:
XS GIS Cut Line= 3
      3769899.61     10547710.19      3769099.61     10547610.19
      3768299.65     10547960.17
#Sta/Elev= 30
  4161.4  358.77  4251.2  345.85  4284.9  340.06  4352.9  335.26  4468.8  319.22
  4514.1  310.57  4595.7  299.93    4625  295.13  4715.7  282.77  4768.6  280.71
  4786.2  277.52  4849.2  275.12  4970.4  275.06  4976.6  271.36  4982.1  274.81
    4997  270.73  4999.7  270.23    5003  270.73  5022.2  274.94  5087.7   273.1
  5104.5   275.4  5127.8  273.97  5151.2  275.56  5164.1  274.01  5589.8  273.87
  5657.2  279.68    5688  285.47  5732.9  290.77    5803  303.27  5840.8  306.28
#Mann= 8 ,-1 , 0
  4161.4     .05       0  4251.2     .16       0  4468.8     .12       0
  4595.7     .05       0    4625     .16       0    4997     .07       0
    5003     .16       0    5688     .16       0
Bank Sta=4982.1,5022.2
XS Rating Curve= 0 ,0
Exp/Cntr=0.3,0.1

Type RM Length L Ch R = 1 ,13002   ,950,950,950
BEGIN DESCRIPTION:
Mapping XS 40d2e9ba
END DESCRIPTION:
XS GIS Cut Line= 4
      3770206.61     10547146.72      3769659.71     10546877.61
      3768965.26       10547329.      3767473.36     10547675.95
#Sta/Elev= 30
  3701.2  342.15  3866.9  333.18    4086     312  4143.7  309.06  4198.4  303.26
  4210.5  301.95  4226.4  288.67  4271.4  290.72  4320.7  281.91  4477.8  272.33
    4985  273.35  4990.9  267.56  4997.1  267.21  4999.8  266.71  5003.1  267.21
  5006.1  270.37  5021.2  273.37  5078.5  272.99  5086.1  269.97  5129.9  273.19
  5319.3  270.55  5596.5  275.59  5801.9     292  5986.7   289.5  6017.5  289.81
    6038  286.48  6058.5  290.13  6263.9  300.05  6428.1  312.07  6670.7  323.93
#Mann= 6 ,-1 , 0
  3701.2     .16       0  4143.7     .16       0  4198.4     .16       0
  4997.1     .07       0  5003.1     .16       0  5986.7     .16       0
Bank Sta=4985,5021.2
XS Rating Curve= 0 ,0
Exp/Cntr=0.3,0.1

Type RM Length L Ch R = 1 ,12052   ,887,887,887
BEGIN DESCRIPTION:
UNT094 IN BECR 15.0
END DESCRIPTION:
XS GIS Cut Line= 3
      3770223.96     10545679.69       3769260.4     10546044.28
      3768001.69     10547259.59
#Sta/Elev= 30
  3150.5  359.92  3358.3  334.84  3565.9  295.36  3711.1  285.45  3869.3  280.66
  4517.8  275.38  4546.1  272.57  4560.2  275.78  4871.5  268.51  4984.7  271.13
  4995.8   267.2  4998.6   266.7  5001.8   267.2    5013  271.46  5133.1  270.05
  5154.5  272.53  5189.7  267.61  5203.9     271  5210.8  276.09  5232.2   278.5
  5331.2  283.65  5373.7  282.09  5408.9  286.14    5501  289.83  5522.1   287.7
  5571.7  291.73  5585.8  288.97    5607  293.44  5669.7   295.4  5930.4  308.69
#Mann= 7 ,-1 , 0
  3150.5     .16       0  3565.9     .05       0  3711.1     .16       0
  4995.8     .07       0  5001.8     .16       0  5408.9     .16       0
  5669.7     .05       0
#XS Ineff= 2 , 0
         4716.48  292.17
Permanent Ineff=
       F       F
Bank Sta=4984.7,5013
XS Rating Curve= 0 ,0
Exp/Cntr=0.3,0.1

Type RM Length L Ch R = 1 ,11165   ,540,540,540
BEGIN DESCRIPTION:
UNT094 IN BECR 14.0
END DESCRIPTION:
XS GIS Cut Line= 3
      3770149.59     10545560.19      3768599.61     10545960.19
      3767926.25     10546604.33
#Sta/Elev= 30
  3400.3  354.14  3534.5  340.61  3545.2  336.44  3656.9  324.92  3738.2  313.53
  3772.1  305.08  3825.6  300.25    3958  285.18  4030.3  281.35  4247.1  276.99
  4918.4  271.23  4937.5  268.23  4983.3  267.97  5005.1  262.93  5007.9  262.43
  5011.1  262.93  5050.6  274.02  5057.5  271.42  5078.9  275.35  5085.8  266.19
    5100  263.12  5142.4  263.11  5149.7  269.97  5156.6  271.19  5163.8  282.19
    5178  283.91  5397.2  301.73  5545.6  307.48  5616.4  307.29  5932.9  315.18
#Mann= 5 ,-1 , 0
  3400.3     .16       0  3825.6     .16       0  5005.1     .07       0
  5011.1     .16       0  5616.4     .05       0
#XS Ineff= 2 , 0
         4805.11  285.03
Permanent Ineff=
       F       F
Bank Sta=4918.4,5050.6
XS Rating Curve= 0 ,0
Exp/Cntr=0.3,0.1

Type RM Length L Ch R = 1 ,10625   ,519,519,519
BEGIN DESCRIPTION:
UNT094 IN BECR 13.0
END DESCRIPTION:
XS GIS Cut Line= 3
      3768899.62     10544960.18      3768399.61     10545560.19
      3768199.58     10545910.23
#Sta/Elev= 30
  4247.2  303.97  4285.2  299.53  4303.7  295.83  4375.4  285.16  4396.3  280.35
  4431.4  275.84  4595.4  271.73  4780.3  270.03  4786.8  272.31  4801.1  270.19
  4807.6  272.09  4815.4  269.73  4821.9  271.08  4829.7  269.45  4836.2  270.63
  4879.2  269.02  4893.5  266.01  4907.8  268.75  4978.1  269.19  4997.3  261.77
    5000  261.27  5003.3  261.77  5041.9  270.46  5079.3  269.78  5108.9  265.65
  5154.2  275.12    5219  284.02  5240.6  284.31  5293.1   288.9  5431.4  299.81
#Mann= 7 ,-1 , 0
  4247.2     .05       0  4285.2     .16       0  4303.7     .05       0
  4396.3     .16       0  4997.3     .07       0  5003.3     .16       0
  5293.1     .16       0
#XS Ineff= 2 , 0
         4608.86  277.33
Permanent Ineff=
       F       F
Bank Sta=4978.1,5041.9
XS Rating Curve= 0 ,0
Exp/Cntr=0.3,0.1

Type RM Length L Ch R = 1 ,10106   ,565,565,565
BEGIN DESCRIPTION:
UNT094 IN BECR 12.0
END DESCRIPTION:
XS GIS Cut Line= 3
       3768849.6     10544910.19      3768149.61     10545110.19
      3767999.62     10545860.14
#Sta/Elev= 30
  4272.9  304.66  4283.3  303.78  4345.7  292.82  4401.6  286.25  4408.1  284.55
  4469.2  275.15  4614.8  267.79    4620  268.58  4731.8  266.71  4765.6  267.66
  4969.7  268.24    4984  267.59  4990.5  266.15  4998.3  261.69  5008.1  261.56
  5010.8  261.06  5014.1  261.56  5021.3  266.13  5072.3  268.33    5266  267.58
  5357.8  269.04  5378.2     266  5398.6  268.34    5470  269.62  5589.7  275.66
  5602.6  276.45    5623  280.15  5668.6  285.76  5735.2  295.39  5765.7  298.57
#Mann= 6 ,-1 , 0
  4272.9     .16       0  4408.1     .16       0  5008.1     .07       0
  5014.1     .16       0  5589.7     .05       0  5668.6     .16       0
#XS Ineff= 2 , 0
                         5271.82          276.08
Permanent Ineff=
       F       F
Bank Sta=4969.7,5072.3
XS Rating Curve= 0 ,0
Exp/Cntr=0.3,0.1

Type RM Length L Ch R = 1 ,9541    ,567,567,567
BEGIN DESCRIPTION:
UNT094 IN BECR 11.0
END DESCRIPTION:
XS GIS Cut Line= 3
      3768599.61     10544310.19      3767799.61     10544810.19
      3766999.65      10544660.2
#Sta/Elev= 30
  4046.2  295.77  4053.9  293.21  4075.1  291.08  4081.6   287.8  4146.6  280.23
  4184.8  276.96  4285.4  273.65  4482.3  266.71  4683.6  264.59  4892.7  266.21
  4904.9  266.17  4960.7  266.59  4986.7  260.81    5007  260.68  5009.7  260.18
    5013  260.68  5015.9  264.15    5021  265.76  5073.5  266.74  5213.4  265.24
  5283.8   262.4  5288.9  264.71    5305  265.32  5498.3  265.78  5528.8   264.4
    5539  261.27  5549.2  266.41  5579.7   264.8    5690  277.57  5803.5  293.91
#Mann= 9 ,-1 , 0
  4046.2     .16       0  4146.6     .12       0  4285.4     .07       0
  4482.3     .12       0  4892.7     .07       0  4904.9     .12       0
    5007     .07       0    5013     .12       0    5690     .16       0
Bank Sta=4960.7,5073.5
XS Rating Curve= 0 ,0
Exp/Cntr=0.3,0.1

Type RM Length L Ch R = 1 ,8974    ,745,745,745
BEGIN DESCRIPTION:
UNT094 IN BECR 10.0
END DESCRIPTION:
XS GIS Cut Line= 3
      3768878.47     10543674.47      3767498.25     10544585.94
      3766526.07      10544646.7
#Sta/Elev= 30
  3500.8  317.34  3642.3  311.55  3756.6  302.06  4000.4  295.07    4154  288.85
    4160  286.42  4218.4  281.06  4298.5  274.98  4506.1  267.42  4716.9  263.01
  4877.4  264.76  4961.5  264.77  4984.8  263.91  4994.4  259.88  4997.2  259.38
  5000.4  259.88  5011.8  260.52  5020.9  264.95    5042  265.91  5203.6  263.84
  5213.6  261.48  5233.6  263.76  5343.8  265.16  5363.9  261.87  5373.9  265.88
    5444  264.45    5513  273.35  5714.6  301.65  5971.3  309.41  6128.9  308.57
#Mann= 8 ,-1 , 0
  3500.8     .16       0  4000.4     .12       0  4218.4     .07       0
  4877.4     .12       0  4994.4     .07       0  5000.4     .12       0
    5513     .16       0  5971.3     .05       0
Bank Sta=4961.5,5042
XS Rating Curve= 0 ,0
Exp/Cntr=0.3,0.1

Type RM Length L Ch R = 1 ,8229    ,1157,1157,1157
BEGIN DESCRIPTION:
UNT094 IN BECR 9.0
END DESCRIPTION:
XS GIS Cut Line= 3
      3768199.65     10543710.16      3767249.61     10544260.19
       3766899.6     10544510.19
#Sta/Elev= 30
  3870.6  301.78  3921.6  298.36  3974.6  287.72  4061.8  276.65  4119.6  268.92
  4144.6   268.2    4240  262.45  4296.1  261.57  4360.7  263.92  4409.2  260.91
  4719.8  262.38  4783.7  262.49  4837.3  262.82  4917.4  264.45  4945.3  261.18
  4954.7  263.57  4960.5  260.63  4965.5  264.07  4971.4  264.07  4990.5  262.21
  4993.6  258.51  4996.4  258.01  4999.6  258.51  5017.5  261.07  5026.1   265.7
  5079.9   267.5  5168.7  270.22  5219.1  274.88  5334.6  293.03  5398.5  299.72
#Mann= 11 ,-1 , 0
  3870.6     .16       0  4061.8     .12       0  4144.6     .07       0
    4240     .12       0  4409.2     .07       0  4719.8     .12       0
  4783.7     .07       0  4837.3     .12       0  4993.6     .07       0
  4999.6     .12       0  5079.9     .16       0
Bank Sta=4971.4,5026.1
XS Rating Curve= 0 ,0
Exp/Cntr=0.3,0.1

Type RM Length L Ch R = 1 ,7072    ,616,616,616
BEGIN DESCRIPTION:
UNT094 IN BECR 8.0
END DESCRIPTION:
XS GIS Cut Line= 3
       3767999.6     10542960.19      3767199.61     10543510.19
      3766749.61     10543860.18
#Sta/Elev= 30
  4004.3  294.69  4047.6   288.3  4068.6  282.53  4119.3  275.43  4127.3  272.81
  4256.7  263.74  4298.6  264.15  4477.8  257.82  4486.7  257.76  4492.7  259.95
  4522.5  257.78  4537.4  259.73  4731.6  258.78  4975.1   261.1  4993.8  256.59
  4996.6  256.09  4999.8  256.59  5025.8  261.68  5096.4  260.14  5195.9  263.01
  5280.2  271.01  5317.2  272.64  5324.4  275.61  5338.9  274.95  5345.2  277.38
    5395  282.87  5403.1  285.28  5409.5  284.06  5517.2  301.43  5545.2  303.48
#Mann= 5 ,-1 , 0
  4004.3     .16       0  4127.3     .12       0  4993.8     .07       0
  4999.8     .12       0  5280.2     .16       0
Bank Sta=4975.1,5025.8
XS Rating Curve= 0 ,0
Exp/Cntr=0.3,0.1

Type RM Length L Ch R = 1 ,6456    ,538,538,538
BEGIN DESCRIPTION:
UNT094 IN BECR 7.0
END DESCRIPTION:
XS GIS Cut Line= 3
      3768299.62     10542710.19      3766899.61     10543410.19
      3766549.58      10543610.2
#Sta/Elev= 30
  3445.2  313.84  3677.2   301.9  3744.3  299.98  3749.9  301.25  3766.6  299.37
  3772.2  301.28  3794.6  300.74  3847.7  295.27  3937.1   277.1    4001  271.37
  4093.7  263.58  4227.8  258.34  4384.4  259.22  4473.8  257.72  4526.9  259.71
  4965.7  260.26  4974.1     260  4979.7  256.17  4999.1  255.95  5001.8  255.45
  5005.1  255.95  5013.3  256.27  5018.4  260.05  5033.5  261.44  5042.1  267.77
  5077.4  277.44    5217  293.44  5346.9  299.76  5362.5  301.84  5413.6  302.11
#Mann= 6 ,-1 , 0
  3445.2     .16       0    4001     .12       0  4999.1     .07       0
  5005.1     .12       0  5042.1     .16       0  5346.9     .05       0
Bank Sta=4965.7,5033.5
XS Rating Curve= 0 ,0
Exp/Cntr=0.3,0.1
