HEC-RAS study BASSET CREEK.prj: BASSET CREEK Base Level Engineering

--- BASSET CREEK.g01 (geometry) --- (continued)

Type RM Length L Ch R = 1 ,23664   ,463,463,463
BEGIN DESCRIPTION:
BASSET CREEK 51.0
END DESCRIPTION:
XS GIS Cut Line= 3
      3748749.61     10633010.15      3748699.61     10633410.19
      3748449.58     10633710.22
#Sta/Elev= 30
  4558.6  412.17  4629.2  395.38    4682   387.9  4709.8   383.1  4780.4  381.86
    4924  379.44  4931.5   376.7  4951.7  376.29  4959.2     371    4965     371
  4968.9  375.47  4983.2  372.91  4989.7  368.05  4994.5  367.56  4997.3  367.06
  5000.5  367.56  5004.1   369.4  5011.9  367.77  5018.4  375.81  5026.2  371.13
  5039.9   379.5  5061.3  378.91  5067.8  374.97  5075.6  378.71  5095.7  379.97
  5160.3  385.59  5246.2  396.63  5252.7  399.51  5260.5  398.76  5352.3  409.42
#Mann= 6 ,-1 , 0
  4558.6     .12       0    4682     .16       0  4780.4     .12       0
  4994.5     .07       0  5000.5     .12       0  5095.7     .05       0
Bank Sta=4983.2,5018.4
XS Rating Curve= 0 ,0
Exp/Cntr=0.3,0.1

Type RM Length L Ch R = 1 ,23201   ,149,149,149
BEGIN DESCRIPTION:
BASSET CREEK 50.0
END DESCRIPTION:
XS GIS Cut Line= 2
      3748572.31     10632953.69      3748129.61     10633561.32
#Sta/Elev= 30
  4601.5  403.69  4621.9     400  4629.8  400.89    4636   398.7    4659  396.68
  4700.9  389.23  4765.8  381.89  4887.1  375.91  4894.1  373.76    4908  375.02
  4916.5   371.3  4931.1  369.94  4943.6  374.45  4966.7  375.42  4972.9  369.19
  4980.7  365.26  4987.5  371.93  4990.7  364.73  4993.5  364.23  4996.7  364.73
  5002.2  364.86  5008.4  368.69  5016.9  368.59  5023.1  376.29  5094.2   375.7
  5116.7   377.3  5163.4  378.92    5279  385.63  5281.4  385.87  5353.3  392.25
#Mann= 7 ,-1 , 0
  4601.5     .12       0  4990.7     .07       0  4996.7     .12       0
  5116.7     .16       0  5163.4     .12       0    5279     .16       0
  5281.4     .12       0
Bank Sta=4987.5,5008.4
XS Rating Curve= 0 ,0
Exp/Cntr=0.3,0.1

Type RM Length L Ch R = 1 ,23052   ,223,223,223
BEGIN DESCRIPTION:
Mapping XS 39861204
END DESCRIPTION:
XS GIS Cut Line= 3
      3748538.19     10632646.15      3748411.45     10632967.34
       3747977.4     10633514.24
#Sta/Elev= 30
  4406.2  394.33  4453.9  393.79  4548.6  394.05  4553.9  392.03  4571.8  392.95
  4583.7  391.27  4632.4  390.98  4662.2  388.25  4686.5  389.23  4691.9  387.78
  4748.6  385.38    4919  375.63  4954.3   376.9  4975.1  375.35  4986.5  363.86
  4989.3  363.36  4992.5  363.86  4997.5  364.28  5003.9  370.37  5024.7  374.97
  5032.8  375.13    5041  375.03  5210.6   373.8  5293.4  377.84  5312.7  379.58
  5359.6  383.32  5395.8  388.33  5438.1  391.72  5443.9  394.08  5449.7  394.08
#Mann= 10 ,-1 , 0
  4406.2     .12       0  4453.9     .16       0  4748.6     .12       0
  4986.5     .07       0  4992.5     .12       0  5032.8     .16       0
    5041     .12       0  5293.4     .16       0  5312.7     .12       0
  5395.8     .16       0
Bank Sta=4975.1,5024.7
XS Rating Curve= 0 ,0
Exp/Cntr=0.3,0.1

Type RM Length L Ch R = 1 ,22829   ,196,196,196
BEGIN DESCRIPTION:
BASSET CREEK 49.0
END DESCRIPTION:
XS GIS Cut Line= 3
      3748149.61     10632610.19      3748099.61     10633010.19
      3747749.62     10633410.18
#Sta/Elev= 30
  4562.3  400.86  4605.1  396.94  4612.7  395.15  4713.5  382.98  4761.3   378.9
    4847  377.38  4854.6  375.68  4874.7  375.98  4927.6  373.89  4945.3  374.53
  4968.7  373.66  4979.2  371.72  4986.8   370.4  4990.4  362.02  4993.2  361.52
  4996.4  362.02  5015.2  372.12  5071.7   373.2  5121.5  371.53  5145.2  372.64
  5242.1  372.36    5263  373.73  5284.3     372  5383.5  380.81  5418.6  385.01
  5426.2   386.9  5447.1  388.41  5489.8  393.76  5493.6  395.44  5496.9  395.44
#Mann= 4 ,-1 , 0
  4562.3     .16       0  4990.4     .07       0  4996.4     .16       0
  5145.2     .16       0
Bank Sta=4979.2,5015.2
XS Rating Curve= 0 ,0
Exp/Cntr=0.3,0.1

Type RM Length L Ch R = 1 ,22633   ,232,232,232
BEGIN DESCRIPTION:
Mapping XS 7ab7f2c3
END DESCRIPTION:
XS GIS Cut Line= 3
      3748057.29     10632602.74      3747991.31     10632845.81
      3747658.86      10633306.4
#Sta/Elev= 30
  4593.2  397.82  4611.3  393.95    4632  393.33  4652.7  389.65  4787.4  375.47
  4808.2  374.25  4856.6  373.64    4886  371.68  4957.2  372.94  4963.3  371.47
  4971.9  371.57    4978  370.49  4986.1  368.62  4992.7  364.68  4995.9  361.86
  4998.7  361.36  5001.9  361.86  5013.6  367.84  5022.2  370.78  5063.9  371.94
  5072.5  371.65  5084.8  368.69  5093.3  370.58    5108  371.35  5229.5  372.36
  5271.3  374.19  5279.8  375.95  5300.7  376.66  5306.9  378.03  5413.1  384.49
#Mann= 3 ,-1 , 0
  4593.2     .16       0  4995.9     .07       0  5001.9     .16       0
Bank Sta=4978,5022.2
XS Rating Curve= 0 ,0
Exp/Cntr=0.3,0.1

Type RM Length L Ch R = 1 ,22401   ,415,415,415
BEGIN DESCRIPTION:
BASSET CREEK 48.0
END DESCRIPTION:
XS GIS Cut Line= 3
      3748049.62     10632460.17      3747749.61     10632860.19
      3747499.63     10633160.16
#Sta/Elev= 30
  4495.1  412.43  4527.6  408.43  4565.2  403.18  4581.6  402.27  4595.1  399.18
  4652.4  391.59    4667   391.2  4728.8  383.86  4773.2  380.74  4837.8  373.31
  4908.7  369.87  4958.7  370.61  4973.2  368.34  4981.6  368.71  4987.8  361.14
  4999.3  360.17    5002  359.67  5005.3  360.17  5008.8  362.12  5016.6  360.46
  5030.9  360.76  5037.4  364.48  5045.2  364.02  5049.9  367.78  5051.7  369.22
  5286.1  370.72    5329  383.57  5349.8  387.25  5357.7  391.31  5385.6  394.93
#Mann= 7 ,-1 , 0
  4495.1     .16       0  4527.6     .12       0  4565.2     .16       0
  4728.8     .12       0  4999.3     .07       0  5005.3     .12       0
  5049.9     .16       0
Bank Sta=4981.6,5051.7
XS Rating Curve= 0 ,0
Exp/Cntr=0.3,0.1

Type RM Length L Ch R = 1 ,21986   ,455,455,455
BEGIN DESCRIPTION:
BASSET CREEK 47.0
END DESCRIPTION:
XS GIS Cut Line= 3
      3747599.61     10632260.17      3747499.61     10632560.19
      3747149.62     10632910.17
#Sta/Elev= 30
  4705.7  407.64  4726.8  406.39  4758.4  402.98  4779.5  398.95    4790  395.54
  4800.6  395.07  4832.2  386.87  4842.7  385.81  4863.8  381.23  4927.1  372.38
  4958.7  368.87  4969.2  368.98  4979.8  365.42  4990.3  363.63  4997.9  359.08
  5000.6  358.58  5003.9  359.08  5011.4  365.52  5019.3  367.63  5036.1  367.82
  5064.4  366.35  5120.9   367.2  5234.1  366.64  5310.4   367.4  5347.2   368.3
  5375.5  372.73  5417.9  383.55  5446.2   388.9  5474.5  391.66  5516.9  397.87
#Mann= 4 ,-1 , 0
  4705.7     .12       0  4997.9     .07       0  5003.9     .12       0
  5310.4     .16       0
Bank Sta=4979.8,5011.4
XS Rating Curve= 0 ,0
Exp/Cntr=0.3,0.1

Type RM Length L Ch R = 1 ,21531   ,285,285,285
BEGIN DESCRIPTION:
BASSET CREEK 46.0
END DESCRIPTION:
XS GIS Cut Line= 3
      3747449.64     10632160.18      3747149.61     10632260.19
      3746899.59     10632660.22
#Sta/Elev= 30
  4653.7  400.62  4674.8  396.43  4706.4  392.22    4717  389.52  4727.5  389.39
  4738.1  387.08  4780.2  382.88  4832.9  375.95  4959.4   366.4  4977.6   365.9
  4983.5  364.71    4993  354.82  4995.9  353.23  4998.6  352.73  5001.9  353.23
  5005.3  357.76  5014.2  362.78  5019.3  364.19  5041.3  365.37  5093.2  364.06
  5135.6   365.1  5172.2  363.63  5253.8  364.19  5288.4  365.32  5339.7  370.02
  5347.3  371.69  5382.7  374.06  5406.3  377.93  5428.1  383.81  5441.7  385.23
#Mann= 5 ,-1 , 0
  4653.7     .12       0  4995.9     .07       0  5001.9     .12       0
  5019.3     .16       0  5253.8     .12       0
Bank Sta=4983.5,5019.3
XS Rating Curve= 0 ,0
Exp/Cntr=0.3,0.1

Type RM Length L Ch R = 1 ,21246   ,165,165,165
BEGIN DESCRIPTION:
Mapping XS 1f3d6573
END DESCRIPTION:
XS GIS Cut Line= 3
      3746932.96     10631885.27      3746866.99     10632183.86
       3746828.8     10632621.41
#Sta/Elev= 30
  4645.8  380.37  4661.1  379.77  4680.5  377.21  4685.6  377.89    4702  375.64
  4734.4  373.65  4763.5  370.68    4778  370.99  4785.3   369.5  4804.5  367.08
  4814.7  367.04  4855.7  363.57  4957.9  362.97    4976   363.7    4981  363.07
  4995.1  350.28  4997.8  349.78  5001.1  350.28  5008.1  359.45  5018.2  363.87
  5058.3  362.55    5159  362.66  5211.4  362.77    5249  363.95  5299.2  369.24
  5309.3  371.21  5319.1  371.17  5329.3  373.28  5369.5  376.74  5390.8  380.32
#Mann= 5 ,-1 , 0
  4645.8     .05       0  4785.3     .16       0  4995.1     .07       0
  5001.1     .16       0    5159     .12       0
Bank Sta=4981,5018.2
XS Rating Curve= 0 ,0
Exp/Cntr=0.3,0.1

Type RM Length L Ch R = 1 ,21081   ,139,139,139
BEGIN DESCRIPTION:
BASSET CREEK 45.0
END DESCRIPTION:
XS GIS Cut Line= 3
      3746799.61     10631810.17      3746699.61     10632210.19
      3746749.61     10632560.21
#Sta/Elev= 30
  4586.6  391.85  4627.8  390.83  4687.1  384.49  4692.3  384.85  4728.3  379.02
  4733.5  380.28  4751.5  376.21  4761.7  375.22  4769.6  372.93  4782.5  372.09
  4792.8  369.51  4823.7  366.32  4864.9  362.64  4896.2  362.03  4921.3  361.93
  4980.9  362.75  4988.6  358.58  4993.4  349.91  4996.1  349.41  4999.4  349.91
    5009  353.68  5019.1  362.55  5139.9  361.62  5160.8  361.36    5176  361.47
  5190.9  361.39  5241.4  366.93  5251.5  366.56  5291.9   372.7  5352.5  377.61
#Mann= 9 ,-1 , 0
  4586.6     .05       0  4761.7     .16       0  4896.2     .05       0
  4921.3     .16       0  4993.4     .07       0  4999.4     .16       0
  5139.9     .05       0  5160.8     .16       0    5176     .12       0
Bank Sta=4980.9,5019.1
XS Rating Curve= 0 ,0
Exp/Cntr=0.3,0.1

Type RM Length L Ch R = 1 ,20942   ,285,285,285
BEGIN DESCRIPTION:
Mapping XS 12cbe93d
END DESCRIPTION:
XS GIS Cut Line= 3
      3746651.72     10631812.31      3746554.49     10632176.92
      3746675.98     10632555.24
#Sta/Elev= 30
  4598.2  386.46  4616.7  383.37  4704.1  376.32  4730.7  372.97  4761.6  371.37
  4771.9  369.48  4824.4  364.47  4881.4  361.59  4906.5  360.85  4980.1  361.35
  4983.8  359.47  4989.5  356.58    4997  351.19  4999.7  350.69    5003  351.19
  5006.9  358.45  5012.2  354.93    5021  361.71  5035.9  361.17    5126   359.9
  5192.2  360.55  5231.1  359.77  5269.1  362.65  5274.3   364.7  5294.1  365.01
  5301.2   365.6  5306.4  367.23  5325.1  368.11  5346.6  370.26  5372.9   371.5
#Mann= 9 ,-1 , 0
  4598.2     .05       0  4730.7     .16       0  4881.4     .05       0
  4983.8     .16       0    4997     .07       0    5003     .16       0
  5035.9     .05       0  5192.2     .16       0  5325.1     .12       0
Bank Sta=4980.1,5006.9
XS Rating Curve= 0 ,0
Exp/Cntr=0.3,0.1

Type RM Length L Ch R = 1 ,20657   ,514,514,514
BEGIN DESCRIPTION:
BASSET CREEK 44.0
END DESCRIPTION:
XS GIS Cut Line= 3
      3746367.43     10631764.51      3746267.61     10632224.54
      3745683.16     10632687.77
#Sta/Elev= 30
  4584.4  389.47  4738.9   374.2  4794.9  374.64  4832.1  372.54  4837.2  375.03
    4846  372.01  4897.2  364.78  4964.3  359.72  4974.5  357.18  4979.6  359.13
  4989.3   356.9  4996.5  347.89  4999.3  347.39  5002.5  347.89  5009.8  359.29
  5023.6  359.75  5030.2  352.89  5050.4  358.03  5163.9  358.03  5363.4  359.27
  5427.7  361.29  5599.2  360.11  5613.7  361.19    5620  368.52  5634.5  367.66
  5640.8   363.4  5664.8  363.43  5684.1  367.26  5698.6  366.19  5800.9  375.79
#Mann= 7 ,-1 , 0
  4584.4     .05       0  4964.3     .16       0  4996.5     .07       0
  5002.5     .16       0  5163.9     .05       0  5363.4     .16       0
  5664.8     .12       0
Bank Sta=4979.6,5009.8
XS Rating Curve= 0 ,0
Exp/Cntr=0.3,0.1

Type RM Length L Ch R = 1 ,20143   ,368,368,368
BEGIN DESCRIPTION:
BASSET CREEK 43.0
END DESCRIPTION:
XS GIS Cut Line= 3
      3746199.64     10631710.16      3745799.61     10632060.19
      3745449.58     10632460.22
#Sta/Elev= 30
  4471.1   388.5  4584.6  379.74  4605.4  375.92  4633.9  372.79  4655.7  372.49
  4662.4  370.46  4698.8  366.74    4726  362.45  4763.1  359.79  4892.5  355.74
  4988.9  356.52  4995.5  348.43  4996.3  346.14  4999.1  345.64  5002.3  346.14
    5006  346.14  5009.8  356.13  5073.4  354.78  5293.6  356.21  5314.4  357.35
  5342.4  363.72  5349.6  366.95  5357.1  364.06    5378  362.62  5385.6  366.37
  5470.1  377.76  5491.9  382.69    5527  387.59  5530.8  390.34  5534.2  390.34
#Mann= 7 ,-1 , 0
  4471.1     .05       0  4698.8     .16       0  4763.1     .05       0
  4892.5     .16       0  4996.3     .07       0  5002.3     .16       0
  5342.4     .12       0
Bank Sta=4988.9,5009.8
XS Rating Curve= 0 ,0
Exp/Cntr=0.3,0.1

Type RM Length L Ch R = 1 ,19775   ,488,488,488
BEGIN DESCRIPTION:
BASSET CREEK 42.0
END DESCRIPTION:
XS GIS Cut Line= 3
      3745949.64     10631760.19      3745549.61     10631787.81
      3745149.65     10631610.21
#Sta/Elev= 30
  4604.7  371.35  4614.2  370.89    4661  365.38  4673.6  363.22  4678.6  363.79
  4684.9  361.78    4715  356.16    4735  354.44  4805.2  353.41  4826.4  354.24
  4895.4  353.03  4949.2  353.48  4975.6  353.21  4985.6  350.48  4995.7  345.22
  5008.4  345.99  5011.6  354.17  5017.1   345.1  5027.6  349.64  5034.9  348.13
  5037.4  344.86  5040.1  344.36  5043.4  344.86  5063.6  346.04  5071.3  352.41
  5105.6  352.74  5162.2  356.31  5278.5  367.51  5335.9  371.39  5443.3  380.59
#Mann= 7 ,-1 , 0
  4604.7     .05       0  4614.2     .16       0    4661     .05       0
  4949.2     .16       0  5037.4     .07       0  5043.4     .16       0
  5105.6     .05       0
Bank Sta=5027.6,5071.3
XS Rating Curve= 0 ,0
Exp/Cntr=0.3,0.1

Type RM Length L Ch R = 1 ,19287   ,469,469,469
BEGIN DESCRIPTION:
BASSET CREEK 41.0
END DESCRIPTION:
XS GIS Cut Line= 3
      3745899.57     10631710.16      3745499.61     10631360.19
      3745149.58      10631460.2
#Sta/Elev= 30
  4457.8  367.01  4461.1  367.01  4464.9  364.03  4485.8  362.38  4493.3  360.62
    4500  360.97  4514.2  359.79  4536.1  356.16  4556.9  355.69  4571.2  354.18
  4748.7  352.01  4776.7  352.84    4798  351.36  4890.1   350.4  4939.4  350.56
  4975.5  351.65  4991.9  350.62  4996.7  342.03  4999.4  341.53  5002.7  342.03
  5006.2  350.35  5011.4  344.41  5020.5  350.86  5051.7  351.69  5072.5  353.24
  5145.3  362.39  5224.6  367.91  5263.6  369.68  5270.1  371.43  5353.3  378.77
#Mann= 3 ,-1 , 0
  4457.8     .05       0  4996.7     .03       0  5002.7     .05       0
Bank Sta=4991.9,5006.2
XS Rating Curve= 0 ,0
Exp/Cntr=0.3,0.1

Type RM Length L Ch R = 1 ,18818   ,334,334,334
BEGIN DESCRIPTION:
BASSET CREEK 40.0
END DESCRIPTION:
XS GIS Cut Line= 3
      3745949.63      10631160.2      3745549.61     10630910.19
      3745149.64     10631110.17
#Sta/Elev= 30
  4529.6  366.32  4637.5  357.75    4647  357.68  4695.3  353.06  4762.5  348.48
  4789.6   347.7  4899.3   347.8  4914.6   347.1  4972.4  348.62  4993.7  346.72
  4995.4  341.03  4998.1  340.53  5001.4  341.03  5004.1  341.03  5009.7  346.63
  5015.3  344.56  5023.7   348.2  5037.7  348.78  5143.9  347.63  5157.8  348.36
  5166.2  350.77  5180.2  350.57  5188.6  348.99  5202.6  347.78  5216.5  348.72
  5314.4  350.74  5336.7  351.85  5381.5  355.71  5417.8   361.2  5448.5  364.05
#Mann= 3 ,-1 , 0
  4529.6     .05       0  4995.4     .03       0  5001.4     .05       0
Bank Sta=4993.7,5009.7
XS Rating Curve= 0 ,0
Exp/Cntr=0.3,0.1

Type RM Length L Ch R = 1 ,18484   ,122,122,122
BEGIN DESCRIPTION:
Mapping XS 72c2ebeb
END DESCRIPTION:
XS GIS Cut Line= 2
      3745981.54     10630713.77      3744287.11     10630241.55
#Sta/Elev= 30
  4546.7   349.1  4611.7     349  4808.2  346.14  4974.3   346.6    4984  342.99
  4989.2  346.93  4992.1  337.47  4994.8  336.97  4998.1  337.47  5005.5  338.07
  5015.8  346.61  5175.7  343.99  5541.9  343.46  5570.1  343.73  5640.1  343.54
    5696  343.07  5711.4  344.67  5741.7  343.29  5803.8  343.16  5843.3   347.9
  5856.7  346.71  5921.9  349.85  5956.1  353.49  5995.5   352.8  6029.7  355.31
  6126.6  355.08  6182.1  355.76  6199.3  357.55  6235.9  357.16  6305.7  357.81
#Mann= 10 ,-1 , 0
  4546.7     .08       0  4611.7     .05       0  4992.1     .03       0
  4998.1     .05       0  5541.9     .16       0  5570.1     .05       0
  5640.1     .08       0  5741.7     .05       0  5843.3     .08       0
  6235.9     .05       0
Bank Sta=4989.2,5015.8
XS Rating Curve= 0 ,0
Exp/Cntr=0.3,0.1

Type RM Length L Ch R = 1 ,18362   ,277,277,277
BEGIN DESCRIPTION:
BASSET CREEK 39.0
END DESCRIPTION:
XS GIS Cut Line= 2
      3746019.81     10630620.04      3744266.35      10630175.6
#Sta/Elev= 30
  4451.8  350.41  4779.1  345.78  4920.3  344.35  4956.1  345.58  4967.8  345.34
  4978.1  342.56  4985.4  337.36  4988.2  336.86  4991.4  337.36  4997.1  340.36
  5002.3  337.89  5009.1  341.66  5019.4   345.5  5029.7  345.72  5359.8  343.18
  5421.7   343.2    5432  344.63    5463  342.98  5574.8   343.7  5601.9  343.57
  5734.8  343.86    5777  350.68  5906.6  349.35  5934.6  352.53  5975.6  354.18
  6021.7   351.3  6072.5  354.14  6139.5  355.32  6226.6  359.87  6260.7  359.47
#Mann= 8 ,-1 , 0
  4451.8     .08       0  4779.1     .05       0  4985.4     .04       0
  4991.4     .05       0  5574.8     .08       0  5601.9     .05       0
    5777     .08       0  6072.5     .05       0
Bank Sta=4978.1,5009.1
XS Rating Curve= 0 ,0
Exp/Cntr=0.3,0.1

Type RM Length L Ch R = 1 ,18085   ,89,89,89
BEGIN DESCRIPTION:
Mapping XS 44f0a559
END DESCRIPTION:
XS GIS Cut Line= 2
      3746037.14     10630460.31      3744540.61     10630078.36
#Sta/Elev= 30
  4296.6  367.49  4354.3  363.15  4420.4  361.08  4510.9  360.98  4522.9  361.98
  4552.1  359.54  4634.6  359.67  4640.3  356.96  4655.3  355.66  4727.5  354.98
  4768.8  350.33  4856.1  348.93    4872  346.95  4944.2   346.4  4975.2  344.76
  4985.5  342.32  4995.8  335.55    5005  335.53  5007.8  335.03    5011  335.53
  5016.5  339.38  5026.8  343.34  5329.8  341.41    5613  343.29  5651.5  344.06
    5708  347.96  5733.2  347.61  5738.9  350.09  5781.5  353.55  5841.1  357.58
#Mann= 8 ,-1 , 0
  4296.6     .05       0  4420.4      .1       0  4510.9     .08       0
  4856.1     .05       0    5005     .04       0    5011     .05       0
    5613     .08       0  5781.5     .05       0
Bank Sta=4985.5,5026.8
XS Rating Curve= 0 ,0
Exp/Cntr=0.3,0.1

Type RM Length L Ch R = 1 ,17996   ,87,87,87
BEGIN DESCRIPTION:
Mapping XS 0d1a81bd
END DESCRIPTION:
XS GIS Cut Line= 2
      3746030.24     10630390.87       3744513.7     10630026.49
#Sta/Elev= 30
  4250.3  372.03    4346  367.59  4359.6  365.79  4364.7  367.65  4394.9  366.57
  4448.7  369.91  4477.2  366.51  4532.6  364.96  4616.6  357.16  4663.7  356.18
  4700.5  351.36  4705.6  353.11  4771.4  349.96  4981.2   341.4  4991.4  336.61
    5009  335.27  5011.8  334.77    5015  335.27  5022.3  336.05  5032.6  343.95
  5303.5  340.32  5543.5  342.11  5629.1  347.77  5659.9  347.27  5668.2   349.7
  5733.5  357.11  5742.2  360.86  5762.8   361.6  5783.4  359.35    5810  363.56
#Mann= 7 ,-1 , 0
  4250.3     .05       0    4346     .08       0  4771.4     .05       0
    5009     .04       0    5015     .05       0  5543.5     .08       0
  5668.2     .05       0
Bank Sta=4981.2,5032.6
XS Rating Curve= 0 ,0
Exp/Cntr=0.3,0.1

Type RM Length L Ch R = 1 ,17909   ,87,87,87
BEGIN DESCRIPTION:
Mapping XS 48bbfe77
END DESCRIPTION:
XS GIS Cut Line= 2
      3746071.87      10630349.2      3744526.75     10629970.73
#Sta/Elev= 30
  4152.5  375.19  4213.2  375.04  4278.4  373.32  4329.9  374.51  4401.9  369.29
  4466.2  369.21  4494.6  362.54    4577  361.56  4618.1   355.3  4690.3  355.11
  4731.4  349.09  4889.1  347.27  4978.5   342.3  4999.1  335.15  5009.3  335.13
    5012  334.63  5015.3  335.13  5019.7  338.43    5030  342.06  5297.6  339.61
  5476.3  341.56  5534.4  344.45  5565.3  347.83  5594.8  347.81  5606.5   351.4
  5647.7  355.18    5678  361.07  5724.7  361.53  5730.1  364.83  5743.3  367.15
#Mann= 7 ,-1 , 0
  4152.5     .05       0  4213.2     .08       0  4690.3     .05       0
  4889.1     .08       0  5009.3     .07       0  5015.3     .08       0
  5476.3     .08       0
Bank Sta=4978.5,5030
XS Rating Curve= 0 ,0
Exp/Cntr=0.3,0.1

Type RM Length L Ch R = 1 ,17822   ,192,192,192
BEGIN DESCRIPTION:
Mapping XS 0cae0608
END DESCRIPTION:
XS GIS Cut Line= 2
      3746089.22     10630300.59      3744568.35     10629918.63
#Sta/Elev= 30
  4081.8   374.8  4297.9  373.64  4339.2  369.94    4401  367.49  4429.6  364.19
  4434.8  365.45  4470.7  362.07  4676.5  351.04  4841.1  345.21  4906.2  345.36
  4959.6  343.29  4969.7   343.1  4988.7  339.15    4996  335.38  4998.8  334.88
    5002  335.38  5005.7  338.18  5010.8  337.96  5019.7  342.39  5046.8   342.1
    5052  339.19  5060.9   340.6  5108.4  339.84  5262.7  340.06  5357.7   340.7
  5442.4  342.72  5504.6  351.03  5535.2   350.5  5622.9  360.73  5649.9  361.51
#Mann= 7 ,-1 , 0
  4081.8     .08       0  4959.6     .05       0    4996     .03       0
    5002     .05       0  5108.4     .08       0  5262.7     .05       0
  5357.7     .08       0
Bank Sta=4988.7,5005.7
XS Rating Curve= 0 ,0
Exp/Cntr=0.3,0.1

Type RM Length L Ch R = 1 ,17630   ,205,205,205
BEGIN DESCRIPTION:
BASSET CREEK 38.0
END DESCRIPTION:
XS GIS Cut Line= 2
      3745630.88     10630033.22      3744513.71     10629800.77
#Sta/Elev= 30
  4456.7  358.72  4568.7  353.95  4640.6  350.87  4752.6     347  4818.5  345.48
  4990.6     341  4999.3  335.67  5006.6  334.85  5009.3  334.35  5012.6  334.85
  5019.8  341.93  5153.6   339.2  5254.7  338.65  5275.1  339.47  5280.9  341.05
    5286   339.3  5325.9  342.66    5331  341.03    5376  346.81  5381.1  344.88
  5409.2  348.42  5454.3   352.2  5476.1  355.04  5481.2  354.05  5499.8  355.81
  5526.2  359.92  5531.3  358.51  5571.2  362.87  5581.6  361.83  5597.8  363.82
#Mann= 10 ,-1 , 0
  4456.7     .08       0  4568.7     .05       0  4640.6     .08       0
  4752.6     .05       0  4818.5     .16       0  5006.6     .07       0
  5012.6     .16       0  5153.6     .08       0  5409.2     .05       0
  5454.3     .08       0
Bank Sta=4990.6,5019.8
XS Rating Curve= 0 ,0
Exp/Cntr=0.3,0.1

Type RM Length L Ch R = 1 ,17425   ,460,460,460
BEGIN DESCRIPTION:
BASSET CREEK 37.0
END DESCRIPTION:
XS GIS Cut Line= 3
      3745408.71     10629731.14      3744821.86     10629741.56
       3744408.7     10629679.06
#Sta/Elev= 30
  4604.6  361.28  4683.7  355.75  4863.7  347.49  4893.7   344.1  4903.7  344.82
  4913.7  347.12  4923.7  347.15  4933.8  343.34  4953.8  341.78  4983.8  341.36
  4993.8  334.59  5000.8  334.42  5003.5  333.92  5006.8  334.42  5013.8  338.56
  5033.8  340.67  5061.9  340.14  5236.7   338.3  5284.8  340.74  5300.5  342.75
  5305.6  341.41  5356.7  346.96  5369.3  346.29  5433.1  351.97  5438.2  350.93
  5456.2  352.85  5487.1  355.67  5507.3  355.37  5570.8  360.52  5609.4  364.85
#Mann= 6 ,-1 , 0
  4604.6     .12       0  5000.8     .07       0  5006.8     .12       0
  5061.9     .05       0  5356.7     .16       0  5456.2     .05       0
Bank Sta=4983.8,5033.8
XS Rating Curve= 0 ,0
Exp/Cntr=0.3,0.1

Type RM Length L Ch R = 1 ,16965   ,436,436,436
BEGIN DESCRIPTION:
BASSET CREEK 36.0
END DESCRIPTION:
XS GIS Cut Line= 2
      3745186.41     10629251.98      3744144.81     10629491.55
#Sta/Elev= 30
  4639.9  364.91  4658.2   362.7  4722.2  360.22  4829.6  355.55  4882.9   349.4
  4954.7  343.37  4985.5  339.06  4995.8   336.2    5003  332.95  5005.8  332.45
    5009  332.95  5016.3  337.26  5026.5  338.99  5067.6  337.43  5143.5  337.26
  5167.9  337.82  5211.2  337.57  5235.5  336.01  5303.6  336.27  5313.9  337.05
  5326.3  339.28  5334.4   342.4  5375.4  348.99    5412  347.92  5426.7  349.91
  5447.2  350.15  5459.9  353.23  5488.3  354.35  5686.7  374.86  5708.7  375.61
#Mann= 7 ,-1 , 0
  4639.9     .16       0  4722.2     .12       0    5003     .07       0
    5009     .12       0  5143.5     .05       0  5167.9     .16       0
  5686.7     .05       0
Bank Sta=4985.5,5026.5
XS Rating Curve= 0 ,0
Exp/Cntr=0.3,0.1

Type RM Length L Ch R = 1 ,16529   ,393,393,393
BEGIN DESCRIPTION:
BASSET CREEK 35.0
END DESCRIPTION:
XS GIS Cut Line= 2
       3745113.5     10628925.59      3744120.52     10628904.75
#Sta/Elev= 30
  4677.3  366.63  4701.2  365.03  4771.2  356.86  4791.2  353.78  4871.2  345.56
  4921.2  339.15  4961.3  335.87  4981.3  335.83  4991.3  334.27  5001.3  334.17
  5011.3  336.22  5051.3  336.59  5111.3  334.07  5161.3  334.81  5174.7  333.75
  5188.3  332.52  5191.1  332.02  5194.3  332.52  5201.3  334.17  5291.3  334.61
  5331.3  333.88  5411.4  336.95  5441.4  338.99  5451.4  340.99  5471.4  343.23
  5501.4  345.53  5571.4  355.83  5648.1  363.92  5653.1  363.22  5670.5  365.11
#Mann= 3 ,-1 , 0
  4677.3     .16       0  5188.3     .07       0  5194.3     .16       0
Bank Sta=5174.7,5201.3
XS Rating Curve= 0 ,0
Exp/Cntr=0.3,0.1

Type RM Length L Ch R = 1 ,16136   ,490,490,490
BEGIN DESCRIPTION:
BASSET CREEK 34.0
END DESCRIPTION:
XS GIS Cut Line= 3
      3745099.62     10628710.19      3744699.61     10628560.19
      3744449.57     10628510.18
#Sta/Elev= 30
  4559.5  358.09  4574.6  356.02  4629.6   351.4  4654.7  349.76  4660.3   348.5
    4677  347.93  4730.4  342.13  4794.5   337.5  4800.7  335.91  4825.6  334.08
  4855.9  334.44  4879.9  333.23  4886.1  334.04  4954.7  333.91  4965.3  335.05
  4976.9  334.02    4984  330.48  4993.9  329.79  4996.7  329.29  4999.9  329.79
  5007.1  332.35  5017.3  333.99  5027.5  334.83  5058.1  335.06  5098.9  332.29
  5129.5  333.67  5139.7  335.51  5190.7  341.34  5211.1  345.23  5241.7  347.73
#Mann= 5 ,-1 , 0
  4559.5     .16       0  4629.6     .12       0  4660.3     .16       0
  4993.9     .07       0  4999.9     .16       0
Bank Sta=4976.9,5017.3
XS Rating Curve= 0 ,0
Exp/Cntr=0.3,0.1

Type RM Length L Ch R = 1 ,15646   ,497,497,497
BEGIN DESCRIPTION:
BASSET CREEK 33.0
END DESCRIPTION:
XS GIS Cut Line= 3
      3745249.65     10628010.18      3744449.61     10628210.19
      3744299.65     10628310.16
#Sta/Elev= 30
  4158.5  380.81  4181.7  378.81  4210.1  373.04    4223  371.93  4251.3  365.59
  4264.2  364.44  4271.9   362.2    4375  346.09  4429.1  342.02  4436.9   339.9
  4488.4  336.56  4663.6  333.84  4704.9  332.08  4900.7  332.74  4931.6  334.24
    4960  333.85  4965.1  331.86  4990.7  334.12  4996.7  328.42  5008.7  327.02
  5011.5  326.52  5014.7  327.02  5032.7  329.72  5047.8  330.32  5055.3  333.11
  5104.9  341.17  5119.9  342.99  5127.4  342.53  5142.1  346.62  5163.4   350.4
#Mann= 4 ,-1 , 0
  4158.5     .16       0  5008.7     .07       0  5014.7     .16       0
  5142.1     .05       0
Bank Sta=4990.7,5055.3
XS Rating Curve= 0 ,0
Exp/Cntr=0.3,0.1

Type RM Length L Ch R = 1 ,15149   ,581,581,581
BEGIN DESCRIPTION:
BASSET CREEK 32.0
END DESCRIPTION:
XS GIS Cut Line= 3
      3744449.61     10627460.18      3744199.61     10627860.19
      3743799.62     10628210.18
#Sta/Elev= 30
  4525.6  360.55  4575.7  357.58    4597  353.83  4612.3  353.35  4656.8  346.69
  4726.7  336.59  4758.5  332.31  4785.6   330.3  4858.7  329.53  4867.6   330.7
  4947.2  330.99  4968.4  332.61  4983.7   331.4  4989.6  325.86  4991.4  325.68
  4994.1  325.18  4997.4  325.68  5004.4  325.88  5011.1  331.75  5025.3  332.52
  5084.3  331.24  5110.7  330.44  5137.7  331.97  5220.3  338.68  5262.9  341.55
  5337.6  346.05  5344.2  347.44  5380.3  348.75  5469.7  355.66  5528.8  359.86
#Mann= 10 ,-1 , 0
  4525.6     .05       0  4656.8     .08       0  4726.7     .16       0
  4991.4     .07       0  4997.4     .16       0  5084.3     .05       0
  5137.7     .16       0  5220.3     .08       0  5262.9     .05       0
  5469.7     .08       0
Bank Sta=4983.7,5011.1
XS Rating Curve= 0 ,0
Exp/Cntr=0.3,0.1

Type RM Length L Ch R = 1 ,14568   ,134,134,134
BEGIN DESCRIPTION:
Mapping XS 0bc2b8b7
END DESCRIPTION:
XS GIS Cut Line= 3
      3744228.99      10626901.7      3743894.78      10627498.5
      3743801.48     10627702.46
#Sta/Elev= 30
  4433.1  343.63  4488.7  340.97  4517.8   340.8  4542.3     342  4666.8  343.56
  4710.2  339.56  4726.1  340.35  4731.8  339.19  4747.8  339.44  4774.1  337.51
  4812.9  336.83  4834.6     334  4888.2  331.81  4901.3  330.05  4924.2  330.62
  4931.6  329.82  4937.3  327.95  4969.3  327.77  5001.4  322.67  5004.2  322.17
  5007.4  322.67  5012.6  324.22  5018.4  329.51  5161.5  328.45    5190  329.13
  5236.1   332.1  5241.6  333.93  5265.2  337.83  5272.9  341.01  5341.4  342.91
#Mann= 6 ,-1 , 0
  4433.1     .05       0  4517.8     .08       0  4774.1     .05       0
  5001.4     .04       0  5007.4     .05       0  5265.2     .08       0
Bank Sta=4969.3,5018.4
XS Rating Curve= 0 ,0
Exp/Cntr=0.3,0.1

Type RM Length L Ch R = 1 ,14434   ,157,157,157
BEGIN DESCRIPTION:
BASSET CREEK 31.0
END DESCRIPTION:
XS GIS Cut Line= 2
      3744081.42     10626730.24      3743789.01     10627626.97
#Sta/Elev= 30
  4395.9  343.75  4442.8  341.07  4451.9  341.92  4490.5  338.35  4515.7  338.07
  4542.4  336.38  4585.2  336.69  4606.2  334.06  4637.8  331.95  4643.3  333.11
  4648.6  332.16  4675.2  332.77  4680.5   331.9  4700.9  332.97    4771  332.64
  4776.2  331.32  4834.8   331.1  4907.3  329.09  4930.5  328.39  4984.9  328.99
  4996.6  322.62  4999.3  322.12  5002.6  322.62  5005.9  325.42  5016.4  328.51
  5088.5  328.08  5222.9  329.34  5228.2   330.8  5279.4  334.45  5339.1  341.14
#Mann= 6 ,-1 , 0
  4395.9     .05       0  4442.8     .08       0  4907.3     .05       0
  4996.6     .04       0  5002.6     .05       0  5088.5     .08       0
Bank Sta=4984.9,5016.4
XS Rating Curve= 0 ,0
Exp/Cntr=0.3,0.1

Type RM Length L Ch R = 1 ,14277   ,102,102,102
BEGIN DESCRIPTION:
BASSET CREEK 30.0
END DESCRIPTION:
XS GIS Cut Line= 2
        3743936.     10626693.41      3743664.77      10627535.3
#Sta/Elev= 30
  4435.2  355.61  4475.7   354.2  4502.5  351.78  4514.5  352.22  4539.9  348.38
  4557.9  342.18  4571.9  340.08  4578.9  336.59  4598.7  333.62  4626.1  333.28
    4718  332.03  4819.8  329.54  4928.5  327.39  4978.1  327.43  4988.6  320.11
  4996.3   317.9    4999   317.4  5002.3   317.9  5009.7  322.29  5020.2  326.61
  5026.1  327.83  5154.3  327.82  5183.5  331.23  5198.8  333.31  5209.3  333.48
  5218.5  335.65  5250.5  339.62  5261.8  343.53  5272.3  343.38  5319.7  351.06
#Mann= 9 ,-1 , 0
  4435.2     .08       0  4514.5     .05       0  4626.1     .08       0
    4718     .05       0  4819.8     .08       0  4928.5     .05       0
  4996.3     .04       0  5002.3     .05       0  5183.5     .08       0
Bank Sta=4978.1,5020.2
XS Rating Curve= 0 ,0
Exp/Cntr=0.3,0.1

Type RM Length L Ch R = 1 ,14175   ,477,477,477
BEGIN DESCRIPTION:
Mapping XS ef3b9758
END DESCRIPTION:
XS GIS Cut Line= 2
      3743834.02      10626669.5       3743567.2     10627515.52
#Sta/Elev= 30
  4445.9  351.82    4499  349.73  4539.7  346.44  4551.5  342.29  4562.8  339.59
  4582.9   332.9  4593.4  331.76  4705.5  331.04  4748.9  329.01  4834.6  327.35
  4841.4  326.31  4873.7  327.22  4906.1  326.44  4981.4  327.14  4991.9  318.64
  4999.4  317.57  5002.1  317.07  5005.4  317.57  5008.4  325.93  5033.8  326.82
    5078  325.85  5096.7     327  5105.4  326.43  5159.6  332.24  5190.4  334.59
  5207.7  335.41    5213  337.04  5240.1  341.24    5254   345.1    5333  354.38
#Mann= 8 ,-1 , 0
  4445.9     .05       0  4562.8     .08       0  4705.5     .05       0
  4748.9     .16       0  4999.4     .07       0  5005.4     .16       0
    5078     .05       0  5190.4     .08       0
Bank Sta=4981.4,5008.4
XS Rating Curve= 0 ,0
Exp/Cntr=0.3,0.1

Type RM Length L Ch R = 1 ,13698   ,335,335,335
BEGIN DESCRIPTION:
BASSET CREEK 29.0
END DESCRIPTION:
XS GIS Cut Line= 3
      3743321.86     10626557.51      3743311.44     10626883.92
      3743235.06     10627189.44
#Sta/Elev= 30
    4615  341.25  4677.7     334  4687.7   333.6  4717.7   330.3  4727.7  330.11
  4737.7  327.82  4797.8  323.19  4857.8  322.55  4887.8  324.14  4907.8  324.06
  4917.8  325.23  4937.2  324.15  4971.8   324.1  4996.6  317.92  4999.3  317.42
  5002.6  317.92  5007.9  319.36    5013  323.42  5030.5  324.28  5054.2  324.16
  5071.7  327.35    5113   331.1    5123  331.23  5131.6  332.18  5136.7  331.75
  5143.9  332.33  5172.8  335.78  5226.3  340.35    5247  339.96  5256.5  341.03
#Mann= 4 ,-1 , 0
    4615     .12       0  4996.6     .07       0  5002.6     .12       0
    5123     .05       0
Bank Sta=4971.8,5013
XS Rating Curve= 0 ,0
Exp/Cntr=0.3,0.1

Type RM Length L Ch R = 1 ,13363   ,477,477,477
BEGIN DESCRIPTION:
BASSET CREEK 28.0
END DESCRIPTION:
XS GIS Cut Line= 3
      3742699.59     10626510.17      3742999.61     10626910.19
      3742999.61     10627160.16
#Sta/Elev= 30
  4515.1  363.15  4522.7  363.04    4537  362.19  4543.2  359.21    4587  357.17
  4651.6  351.64    4687  346.77  4715.1   341.3  4722.4  338.21  4728.7  338.38
  4765.1  332.34  4778.7  328.71  4915.1   323.5    4937  320.46  4943.2  323.09
  4951.6  319.67  4972.4  322.51    4987  318.52  4993.2  318.47  5001.6  315.29
  5004.8  312.51  5007.6  312.01  5010.8  312.51    5012  322.24  5065.1  322.46
  5095.1  324.84  5115.1  328.96  5125.1  334.23  5132.9  334.53  5265.1  336.01
#Mann= 5 ,-1 , 0
  4515.1     .08       0  4522.7     .12       0  5004.8     .07       0
  5010.8     .12       0  5132.9     .16       0
Bank Sta=4993.2,5012
XS Rating Curve= 0 ,0
Exp/Cntr=0.3,0.1

Type RM Length L Ch R = 1 ,12886   ,438,438,438
BEGIN DESCRIPTION:
Mapping XS 647055c8
END DESCRIPTION:
XS GIS Cut Line= 2
      3742446.94       10626679.      3742689.35     10627336.96
#Sta/Elev= 30
  4686.4  363.09  4698.3   361.5  4706.1  357.53  4722.6  355.76  4751.6  351.44
  4822.6  345.21  4836.9  345.12    4853  341.61  4858.4  343.09  4868.8  339.53
  4883.5  339.12  4890.2  335.69  4908.6  331.29  4954.1  324.12  4986.1  321.46
  4994.6  313.48    4997  309.47  4999.7  308.97    5003  309.47  5025.1  312.08
  5030.4  318.08  5039.4  320.98  5141.5  322.75  5166.7   324.7  5177.9  327.06
  5227.6  330.52  5252.6  334.06    5258   335.9  5327.1  341.54  5387.6  344.75
#Mann= 5 ,-1 , 0
  4686.4     .05       0  4722.6     .12       0    4997     .07       0
    5003     .12       0  5252.6     .16       0
Bank Sta=4986.1,5039.4
XS Rating Curve= 0 ,0
Exp/Cntr=0.3,0.1

Type RM Length L Ch R = 1 ,12448   ,401,401,401
BEGIN DESCRIPTION:
BASSET CREEK 26.0
END DESCRIPTION:
XS GIS Cut Line= 3
       3742199.6     10626810.23      3742149.61     10627060.19
      3742199.62     10627360.24
#Sta/Elev= 30
  4754.6  358.88  4764.8  358.27  4780.6  355.49  4815.8  347.46  4825.9  343.26
  4856.5   335.8  4866.7  331.49  4876.9  330.96  4887.1  326.75  4897.3  325.33
  4917.7  319.38  4927.9  318.74  4948.3  319.91  4958.5  318.86  4968.7  320.66
  4978.9  319.77  4989.1  309.14  4996.3  305.85  4999.1  305.35  5002.3  305.85
    5007  307.33    5012  307.33  5029.8  315.11  5037.4  320.86  5110.9  319.71
  5164.1  322.38  5202.1  325.91  5212.3  328.19  5232.5  329.33  5313.7  337.45
#Mann= 4 ,-1 , 0
  4754.6     .05       0  4780.6     .12       0  4996.3     .07       0
  5002.3     .12       0
Bank Sta=4978.9,5037.4
XS Rating Curve= 0 ,0
Exp/Cntr=0.3,0.1

Type RM Length L Ch R = 1 ,12047   ,351,351,351
BEGIN DESCRIPTION:
BASSET CREEK 25.0
END DESCRIPTION:
XS GIS Cut Line= 3
      3741949.59     10626710.22      3741799.61     10626960.19
      3741649.62     10627260.17
#Sta/Elev= 30
  4721.9  355.64  4729.6  356.19  4745.2  354.79  4815.2  337.58  4824.9  336.26
  4830.7  332.83    4889  323.03  4896.8  320.61  4920.1  318.59  4947.3  319.07
  4955.1  320.94  4962.9  318.42  4968.7  318.67  4978.4  308.72  4987.1  303.64
  4989.8  303.14  4993.1  303.64  5005.6  303.96  5010.5   308.4  5016.2   308.4
  5021.8  312.01  5027.4  311.61  5035.8  318.82  5066.5  318.17  5125.2  320.36
  5147.6  323.44  5161.6  323.71  5272.6  335.59  5326.5  339.97  5348.8   340.6
#Mann= 4 ,-1 , 0
  4721.9     .12       0  4987.1     .07       0  4993.1     .12       0
  5272.6     .05       0
Bank Sta=4978.4,5010.5
XS Rating Curve= 0 ,0
Exp/Cntr=0.3,0.1

Type RM Length L Ch R = 1 ,11696   ,516,516,516
BEGIN DESCRIPTION:
Mapping XS 14306612
END DESCRIPTION:
XS GIS Cut Line= 2
      3741492.07     10626357.81      3741453.01     10627251.86
#Sta/Elev= 30
  4481.8  348.22  4492.3  347.31  4504.2  344.86  4534.2  341.88  4594.3  340.37
  4634.3  331.89  4656.1  324.63  4684.4  320.53  4704.4  319.51  4724.4  315.53
  4734.4  306.16  4744.4   306.4  4764.4  312.77  4774.5  318.74  4834.5  318.83
  4874.6  316.82  4934.6  316.04  4974.6   318.1  4984.7  306.91  4991.7  302.43
  4994.4  301.93  4997.7  302.43  5004.7  302.56  5014.7  306.06  5034.7  319.08
  5044.7  322.92  5054.7  324.64  5214.9  335.29    5295  338.89  5376.7  339.95
#Mann= 4 ,-1 , 0
  4481.8     .05       0  4492.3     .12       0  4991.7     .07       0
  4997.7     .12       0
Bank Sta=4974.6,5034.7
XS Rating Curve= 0 ,0
Exp/Cntr=0.3,0.1

Type RM Length L Ch R = 1 ,11180   ,476,476,476
BEGIN DESCRIPTION:
BASSET CREEK 23.0
END DESCRIPTION:
XS GIS Cut Line= 2
      3741223.54     10626370.92      3740849.05     10626885.84
#Sta/Elev= 30
  4745.8  345.76  4773.3  342.36  4827.1  339.71  4856.2  339.61  4862.7  336.59
  4883.5  334.83    4892  330.28  4898.2  329.32  4905.6  322.26  4912.9  320.13
  4927.6  318.26  4933.8  318.84  4948.5  315.25  4955.1  315.44  4977.8  303.41
    4984  304.12  4989.2  298.52  4991.9  298.02  4995.2  298.52  5004.9  298.69
  5013.4  303.44  5028.1  305.68  5034.2  309.49  5041.7   309.6  5048.9  316.03
  5128.2  314.65  5177.7  315.86    5321  324.69  5341.8   324.7  5382.5  328.83
#Mann= 4 ,-1 , 0
  4745.8     .05       0  4773.3     .12       0  4989.2     .07       0
  4995.2     .12       0
Bank Sta=4984,5013.4
XS Rating Curve= 0 ,0
Exp/Cntr=0.3,0.1

Type RM Length L Ch R = 1 ,10704   ,494,494,494
BEGIN DESCRIPTION:
BASSET CREEK 22.0
END DESCRIPTION:
XS GIS Cut Line= 3
      3741099.64     10626210.17      3740649.61     10626510.19
      3740549.62     10626760.17
#Sta/Elev= 30
  4476.7  354.56  4490.3  353.44  4499.3  348.72  4544.4  343.07  4584.9     336
  4613.4  334.67  4628.5  329.99  4649.5  328.18    4657  324.98  4685.6  319.75
  4706.6  318.91  4736.6  314.62  4945.5  313.85    4953  312.73    4959   302.6
    4968  301.94  4981.5   296.4    5001  296.07  5003.8  295.57    5007  296.07
  5010.1  300.66  5020.3  300.92    5027  304.02  5032.4  312.66  5039.1  313.84
  5080.8   314.1  5157.6  322.18  5179.1  321.08  5188.5  324.29  5286.8  337.69
#Mann= 4 ,-1 , 0
  4476.7     .05       0  4544.4     .12       0    5001     .07       0
    5007     .12       0
Bank Sta=4968,5010.1
XS Rating Curve= 0 ,0
Exp/Cntr=0.3,0.1

Type RM Length L Ch R = 1 ,10210   ,475,475,475
BEGIN DESCRIPTION:
BASSET CREEK 21.0
END DESCRIPTION:
XS GIS Cut Line= 3
       3740999.6      10625960.2      3740549.61     10626210.19
      3740299.62     10626360.18
#Sta/Elev= 30
  4489.2  355.83  4492.2  355.82  4524.6  353.82  4546.4  350.12  4562.4  349.09
  4569.3   346.1  4584.1  344.35  4605.9  337.88  4627.6  333.02  4649.3  330.28
  4703.1   319.1  4708.8  320.02    4718  317.13  4740.9  314.07  4820.9  311.56
  4946.8  311.22  4958.2  300.48  4968.5  299.87  4981.1  294.53  4990.2  295.34
  5008.7  294.44  5011.5  293.94  5014.7  294.44  5017.6  296.71  5027.3  297.76
    5039  302.78  5048.7  305.39  5054.5  309.25  5143.9   316.2  5295.5  335.84
#Mann= 4 ,-1 , 0
  4489.2     .05       0  4492.2     .12       0  5008.7     .07       0
  5014.7     .12       0
Bank Sta=4946.8,5054.5
XS Rating Curve= 0 ,0
Exp/Cntr=0.3,0.1

Type RM Length L Ch R = 1 ,9735    ,465,465,465
BEGIN DESCRIPTION:
BASSET CREEK 20.0
END DESCRIPTION:
XS GIS Cut Line= 3
      3740549.62     10625710.17      3740349.61     10625910.19
      3740199.61     10626360.18
#Sta/Elev= 30
  4720.6  340.99  4748.9  339.12  4778.4  335.79  4791.3  332.88  4805.5  330.98
  4819.6   326.3  4833.8  324.55    4862  318.36  4890.3  313.99  4918.6  310.73
    4961  310.58  4975.2  307.87  4989.3  294.52  4996.9  293.34  4999.7  292.84
  5002.9  293.34  5006.1  293.34    5014  300.38  5045.6  308.55  5056.2  309.92
  5077.2   309.1  5119.4  310.56  5193.2  310.05  5224.8  310.87  5245.9  313.76
    5331  320.73  5393.5  328.77    5404  331.19  5414.6  331.76  5477.8  342.35
#Mann= 5 ,-1 , 0
  4720.6     .16       0  4778.4     .12       0  4996.9     .07       0
  5002.9     .12       0    5331     .16       0
Bank Sta=4961,5045.6
XS Rating Curve= 0 ,0
Exp/Cntr=0.3,0.1

Type RM Length L Ch R = 1 ,9270    ,438,438,438
BEGIN DESCRIPTION:
BASSET CREEK 19.0
END DESCRIPTION:
XS GIS Cut Line= 3
      3740049.61     10625460.22      3739999.61     10625960.19
      3739949.61     10626160.17
#Sta/Elev= 30
  4491.7  351.05  4531.9  347.74  4639.9  327.63  4644.9  328.62  4671.1  323.59
  4722.8  317.34  4740.4  313.62  4777.2  310.68  4823.3  303.63  4840.9  303.01
  4863.5  307.01  4883.6  304.93  4893.7  307.51  4913.8  308.96    4964  308.63
  4974.1   300.2  4984.1  296.75  4991.7  291.91  5001.5  291.87  5004.2  291.37
  5007.5  291.87  5017.4  294.21  5025.1  302.15  5035.4   306.1  5045.7  307.73
  5058.6  307.52  5117.9  312.73  5141.1   316.5  5159.1  316.93  5200.3  323.83
#Mann= 5 ,-1 , 0
  4491.7     .16       0  4671.1     .12       0  4777.2     .16       0
  5001.5     .07       0  5007.5     .16       0
Bank Sta=4964,5045.7
XS Rating Curve= 0 ,0
Exp/Cntr=0.3,0.1

Type RM Length L Ch R = 1 ,8832    ,481,481,481
BEGIN DESCRIPTION:
BASSET CREEK 18.0
END DESCRIPTION:
XS GIS Cut Line= 3
      3739549.61     10625460.16      3739599.61     10625910.19
      3739599.61     10626110.19
#Sta/Elev= 30
  4535.9   359.5  4576.2  352.69  4586.2  349.09  4596.3  348.19  4646.6  335.83
  4656.7  334.37  4686.9  324.49  4696.9  323.08    4717  317.59  4747.2  314.19
  4767.3  313.97  4837.8  308.54    4878  308.29  4928.3  306.06  4938.4  302.65
  4948.5  305.89  4968.6  306.03  4978.6  299.72  4986.2   293.2  5005.7  290.08
  5008.5  289.58  5011.7  290.08  5018.7  296.37  5028.7  302.76  5038.7  307.12
  5048.7  307.75  5078.7  314.05  5138.7  319.69  5148.7  322.11  5188.7  327.39
#Mann= 3 ,-1 , 0
  4535.9     .16       0  5005.7     .07       0  5011.7     .16       0
Bank Sta=4968.6,5038.7
XS Rating Curve= 0 ,0
Exp/Cntr=0.3,0.1

Type RM Length L Ch R = 1 ,8351    ,463,463,463
BEGIN DESCRIPTION:
BASSET CREEK 17.0
END DESCRIPTION:
XS GIS Cut Line= 3
      3739349.62     10625310.15      3739149.61     10625810.19
      3739149.61     10626060.23
#Sta/Elev= 30
    4480  369.22  4489.5  368.82  4494.9  365.77    4510  365.02  4524.5  361.62
  4548.7  359.92  4555.4  356.69  4572.9  353.39  4663.1  338.52  4727.8   329.9
  4749.3  323.97  4781.6   319.3  4793.7  315.42    4857   310.6  4866.4  313.39
  4901.4  306.54  4955.3  303.81  4964.7  297.38  4979.5  296.47    4994  289.62
  4996.8  289.12    5000  289.62  5009.1  290.62  5015.9  296.87  5021.1  296.87
  5038.6  302.38  5058.6  304.89  5088.6  304.77  5108.6  306.64  5268.6  328.62
#Mann= 4 ,-1 , 0
    4480     .05       0    4510     .16       0    4994     .07       0
    5000     .16       0
Bank Sta=4979.5,5015.9
XS Rating Curve= 0 ,0
Exp/Cntr=0.3,0.1

Type RM Length L Ch R = 1 ,7888    ,284,284,284
BEGIN DESCRIPTION:
BASSET CREEK 16.0
END DESCRIPTION:
XS GIS Cut Line= 3
      3739099.63     10625160.16      3738799.61     10625610.19
      3738849.61     10626060.15
#Sta/Elev= 30
  4457.4  367.49    4522  360.03  4529.5   357.1  4552.1  352.82  4637.7  343.18
  4738.4  323.73  4774.4  318.05  4781.9   318.5  4795.5  314.53  4876.6  307.58
  4962.2  302.95  4969.7  301.39  4975.7  295.13  4984.7  295.69  4992.3  286.75
    4995  286.25  4998.3  286.75  5008.3  287.31  5018.4  293.59  5048.6   296.5
  5078.8   303.9  5098.9  300.45    5119  303.56  5129.1  303.87  5139.1   301.7
  5149.2  303.98  5229.7  305.45  5249.8  297.86  5259.9  304.68    5451  325.74
#Mann= 3 ,-1 , 0
  4457.4     .16       0  4992.3     .07       0  4998.3     .16       0
Bank Sta=4984.7,5018.4
XS Rating Curve= 0 ,0
Exp/Cntr=0.3,0.1

Type RM Length L Ch R = 1 ,7604    ,201,201,201
BEGIN DESCRIPTION:
Mapping XS 0a4f5edf
END DESCRIPTION:
XS GIS Cut Line= 3
      3738708.36     10625083.68       3738557.3     10625422.25
      3738505.33     10626066.62
#Sta/Elev= 30
  4561.1  340.15  4688.1   337.6  4693.6  339.36  4776.3  334.16  4791.9  331.64
  4798.2  328.47  4809.1  326.57  4815.2  322.99    4831  320.57  4843.9   314.5
  4852.9  314.51  4874.8  309.68    4919  303.82  4949.8  301.33  4959.9  302.28
  4970.1  300.17  4979.9  293.84    4990  286.29    4997   285.8  4999.8   285.3
    5003   285.8  5010.6  290.14  5030.1  296.52  5060.2   298.3    5089  302.74
  5209.9  303.15  5331.1  306.93  5459.7  313.36  5471.5   315.5  5578.3  319.44
#Mann= 5 ,-1 , 0
  4561.1     .16       0    4997     .07       0    5003     .16       0
  5010.6     .12       0    5089     .16       0
Bank Sta=4979.9,5030.1
XS Rating Curve= 0 ,0
Exp/Cntr=0.3,0.1

Type RM Length L Ch R = 1 ,7403    ,238,238,238
BEGIN DESCRIPTION:
BASSET CREEK 15.0
END DESCRIPTION:
XS GIS Cut Line= 3
      3738549.63     10625210.17      3738399.61     10625410.19
      3738049.64     10625660.16
#Sta/Elev= 30
  4772.3  334.31  4829.6  323.83  4835.9  319.46  4844.2  318.33  4858.8     311
  4866.2  310.54    4915   303.7  4922.3  301.71  4958.8  301.51    4965  297.61
  4979.6  294.35  4985.9  289.81  4994.2  288.07  4997.5  285.19  5000.2  284.69
  5003.5  285.19  5008.8  285.25    5015   291.2  5019.2  292.78  5042.9  295.88
  5059.2  301.76    5101  301.27  5166.1  304.86  5207.9  310.23  5231.2  311.78
  5258.3   316.8  5266.9  316.22  5302.5  319.39  5388.5  329.72  5452.4  340.13
#Mann= 5 ,-1 , 0
  4772.3     .16       0  4866.2     .12       0  4997.5     .07       0
  5003.5     .12       0  5042.9     .16       0
Bank Sta=4979.6,5015
XS Rating Curve= 0 ,0
Exp/Cntr=0.3,0.1

Type RM Length L Ch R = 1 ,7165    ,188,188,188
BEGIN DESCRIPTION:
Mapping XS 1f53a5fd
END DESCRIPTION:
XS GIS Cut Line= 3
      3738565.14     10625008.17      3738317.72      10625200.9
      3737968.74     10625594.15
#Sta/Elev= 30
  4658.6  349.13  4720.8   342.6  4749.7  336.63    4756  337.54  4764.2  334.43
    4785   332.1  4813.9  325.26  4834.7  323.56  4863.7  317.78    4870  318.18
  4919.8   309.8  4942.4  304.91  4967.9  293.69  4974.6  293.69  4977.4  290.84
  4991.7  286.88  4995.3   284.5  4998.1     284  5001.3   284.5  5013.3  289.95
  5026.8  294.25    5041  295.28  5048.5  298.93  5059.2  301.24  5147.2  298.86
    5169  300.63  5204.1  306.13  5317.8  319.31    5466  341.56    5498  342.53
#Mann= 5 ,-1 , 0
  4658.6     .16       0  4995.3     .07       0  5001.3     .16       0
  5013.3     .12       0  5059.2     .16       0
Bank Sta=4974.6,5026.8
XS Rating Curve= 0 ,0
Exp/Cntr=0.3,0.1

Type RM Length L Ch R = 1 ,6977    ,267,267,267
BEGIN DESCRIPTION:
BASSET CREEK 14.0
END DESCRIPTION:
XS GIS Cut Line= 3
      3738399.64     10624960.16      3738138.03     10625193.09
      3737949.58     10625460.23
#Sta/Elev= 30
  4618.1  341.35  4688.8  332.12  4696.3  327.46  4717.2  323.28  4724.7  318.35
  4745.7  311.82  4805.8  302.61  4830.9   299.9  4915.4  299.89  4943.8  295.93
  4951.3  299.13  4968.4  297.55  4972.6  288.57  4978.8  287.59  4984.4   283.8
  4987.2   283.3  4990.4   283.8  5001.5   283.9  5005.6  287.27  5008.3  289.49
  5014.5  288.43    5044     293  5058.8  299.69    5065  298.31  5073.6  301.96
  5151.2  309.48  5231.2  323.27    5246  323.06  5258.5  327.94  5295.3  334.27
#Mann= 5 ,-1 , 0
  4618.1     .16       0  4805.8     .12       0  4984.4     .07       0
  4990.4     .12       0  5005.6     .16       0
Bank Sta=4978.8,5008.3
XS Rating Curve= 0 ,0
Exp/Cntr=0.3,0.1

Type RM Length L Ch R = 1 ,6710    ,286,286,286
BEGIN DESCRIPTION:
Mapping XS cc5cb7da
END DESCRIPTION:
XS GIS Cut Line= 3
      3738471.62     10624827.09      3738049.72     10625064.08
      3737664.43     10625441.57
#Sta/Elev= 30
  4636.4   329.8  4654.4  333.75    4692  334.08  4697.8  336.68  4719.5   336.7
  4729.7  334.04  4735.4  335.92  4751.3  331.76  4757.1   333.3    4773  329.67
  4778.8  331.28  4794.7  326.07  4800.4  327.75    4854  310.76  4909.9  302.39
  4956.7  299.75  4971.3  293.56  4984.1  285.06    4997  283.23  4999.8  282.73
    5003  283.23  5028.7  292.08  5059.3  294.09  5074.6  299.19  5100.6  298.64
    5252  298.23  5315.7  301.09    5549  322.54  5570.1  327.48  5659.7   336.4
#Mann= 5 ,-1 , 0
  4636.4     .16       0  4909.9     .12       0    4997     .07       0
    5003     .12       0  5100.6     .16       0
Bank Sta=4971.3,5028.7
XS Rating Curve= 0 ,0
Exp/Cntr=0.3,0.1

Type RM Length L Ch R = 1 ,6424    ,293,293,293
BEGIN DESCRIPTION:
BASSET CREEK 13.0
END DESCRIPTION:
XS GIS Cut Line= 3
      3738249.63     10624610.17      3738049.61     10624760.19
      3737549.58     10625360.23
#Sta/Elev= 30
  4749.1  333.95  4756.4  332.62  4762.7  329.52  4777.3  327.15  4785.6  322.86
  4806.4  320.08  4812.7  314.21  4827.3  313.31  4849.1  310.14  4862.7  306.87
  4905.5  302.09  4912.7  302.65  4962.7  298.77  4985.6  293.01    4993  282.14
  4995.8  281.64    4999  282.14  5006.3   282.2  5012.8  286.41  5020.6   288.3
  5041.4   298.1  5066.9  298.63  5339.5  297.07  5446.3  299.96  5524.4  305.03
  5610.3  312.92  5616.8  314.68  5709.2  324.17  5737.8  330.31  5780.2   334.1
#Mann= 5 ,-1 , 0
  4749.1     .16       0  4905.5     .12       0    4993     .07       0
    4999     .12       0  5066.9     .16       0
Bank Sta=4962.7,5041.4
XS Rating Curve= 0 ,0
Exp/Cntr=0.3,0.1
