HEC-RAS study BOX CREEK.prj: BOX CREEK Base Level Engineering

--- BOX CREEK.g01 (geometry) --- (continued)

Type RM Length L Ch R = 1 ,104581  ,514,514,514
BEGIN DESCRIPTION:
BOX CREEK 142.0
END DESCRIPTION:
XS GIS Cut Line= 3
      3781649.58     10584860.17      3781049.61     10584560.19
      3780599.56     10584610.19
#Sta/Elev= 30
  4387.3   359.1  4401.2  359.06  4476.7  351.84    4513  346.96  4574.5  342.88
  4580.1  341.44  4686.3   332.5  4767.4  330.18  4884.6   329.8    4977  330.48
    4991  323.12  4996.4  322.76  4999.1  322.26  5002.4  322.76    5005  325.78
  5013.4  328.95  5027.3  329.38  5044.1  329.41    5053   327.9  5068.1   326.9
  5078.2  324.27  5108.4  330.12  5198.9  328.74  5239.2  330.19  5266.1  328.34
  5319.7  328.78  5372.9  333.69  5450.5   348.4  5480.7  351.45  5510.9  351.95
#Mann= 7 ,-1 , 0
  4387.3     .16       0  4884.6     .12       0  4996.4     .07       0
  5002.4     .12       0    5053     .16       0  5266.1     .12       0
  5372.9     .16       0
Bank Sta=4977,5027.3
XS Rating Curve= 0 ,0
Exp/Cntr=0.3,0.1

Type RM Length L Ch R = 1 ,104067  ,351,351,351
BEGIN DESCRIPTION:
BOX CREEK 141.0
END DESCRIPTION:
XS GIS Cut Line= 3
      3781949.63     10584260.19      3780749.61     10584360.19
      3780599.62     10584510.18
#Sta/Elev= 30
  3773.4  377.85  3831.1  373.71  3883.8   363.2  3964.1  350.09  4024.3  343.29
  4054.4  342.46  4084.5  335.94  4164.8  330.96    4210  330.22  4387.8  328.97
  4455.8  328.47  4495.9  331.67  4546.1  332.15  4626.4  328.46  4679.1  328.59
  4696.6  330.11  4789.1  328.67  4877.2  330.08  4977.6  328.07  4981.1  328.07
  4991.7  321.93  5002.9     321  5005.6   320.5  5008.9     321    5020  321.26
  5034.2  328.76  5080.3  340.87  5090.7  345.09    5119  349.44  5189.7  350.66
#Mann= 7 ,-1 , 0
  3773.4     .16       0    4210     .05       0  4387.8     .16       0
  4789.1     .12       0  5002.9     .07       0  5008.9     .12       0
  5080.3     .16       0
Bank Sta=4977.6,5034.2
XS Rating Curve= 0 ,0
Exp/Cntr=0.3,0.1

Type RM Length L Ch R = 1 ,103716  ,440,440,440
BEGIN DESCRIPTION:
BOX CREEK 140.0
END DESCRIPTION:
XS GIS Cut Line= 3
      3781813.13     10584038.59      3780782.27     10584097.19
      3780473.25     10584187.95
#Sta/Elev= 30
  3868.5  371.76  3902.1  365.95  3942.1  357.08  3972.2  354.22  4040.7  352.74
  4082.4  347.63  4092.4  344.76  4122.4  339.88  4222.6  329.64  4282.7  327.73
  4445.4  328.28  4454.6   328.3  4683.3  327.46  4843.6  328.97  4915.4  327.73
  4976.8  328.32  4987.2  322.85  4996.4  321.79  4998.6  320.22  5001.3  319.72
  5004.6  320.22    5008  320.33  5018.4  329.21  5028.9  331.35  5040.2  336.78
  5060.1   341.3    5081  343.73  5133.9   344.3  5185.2  348.12  5223.1  349.02
#Mann= 8 ,-1 , 0
  3868.5     .05       0  4040.7     .16       0  4445.4     .05       0
  4454.6     .16       0  4915.4     .12       0  4998.6     .07       0
  5004.6     .12       0  5133.9     .16       0
Bank Sta=4976.8,5018.4
XS Rating Curve= 0 ,0
Exp/Cntr=0.3,0.1

Type RM Length L Ch R = 1 ,103276  ,169,169,169
BEGIN DESCRIPTION:
BOX CREEK 139.0
END DESCRIPTION:
XS GIS Cut Line= 3
       3781897.2     10583672.56      3781398.07     10583629.15
       3780130.7     10584093.57
#Sta/Elev= 30
  3731.8   371.1  3793.9  367.27  3933.7  360.59  3960.3  350.13  4000.4  344.18
  4186.2  329.05  4282.3  326.97  4374.6  325.91  4399.9  325.37  4801.8  322.31
  4838.2  324.76  4918.5  320.82  4923.8  323.91    4966  322.89  4979.5   326.2
  5001.7  319.58  5004.4  319.08  5007.7  319.58  5029.9  325.88  5035.2  322.88
  5060.4  322.04  5065.7  326.76  5083.2  329.44  5121.4  329.67  5177.1  338.22
  5212.9  348.55  5299.1  349.58  5402.7  343.52    5575  347.37  5582.6  347.74
#Mann= 9 ,-1 , 0
  3731.8     .05       0  3793.9     .16       0  4186.2     .05       0
  4282.3     .16       0  4374.6     .05       0  4399.9     .16       0
  5001.7     .07       0  5007.7     .16       0    5575     .05       0
Bank Sta=4979.5,5029.9
XS Rating Curve= 0 ,0
Exp/Cntr=0.3,0.1

Type RM Length L Ch R = 1 ,103107  ,78,78,78
BEGIN DESCRIPTION:
Mapping XS bbb09f4d
END DESCRIPTION:
XS GIS Cut Line= 3
      3781823.45     10583559.71      3781311.27     10583511.97
      3779823.57     10584010.76
#Sta/Elev= 30
    3789  356.72  3933.5  346.34  4003.8  336.42  4051.1  335.22  4084.1  339.37
  4160.2  340.15  4194.6  337.39  4224.7  329.03  4234.8  328.36  4371.1  326.87
  4500.1  326.09  4582.4  325.57  4776.9  326.24  4937.7  326.89  4969.3  321.78
  4974.5  326.15  4980.2  320.23  5003.1   319.7  5005.8   319.2  5009.1   319.7
  5032.4  326.38  5173.9   327.1  5353.1  332.37  5442.5  329.96  5505.6  331.74
  5644.6   341.2  5700.2  341.85  5726.4  345.67  5731.7  342.78  5872.5  346.06
#Mann= 8 ,-1 , 0
    3789     .16       0  4371.1     .12       0  4500.1     .16       0
  4582.4     .12       0  4776.9     .16       0  5003.1     .07       0
  5009.1     .16       0  5173.9     .05       0
Bank Sta=4974.5,5032.4
XS Rating Curve= 0 ,0
Exp/Cntr=0.3,0.1

Type RM Length L Ch R = 1 ,103029  ,1064,1064,1064
BEGIN DESCRIPTION:
BOX CREEK 138.0
END DESCRIPTION:
XS GIS Cut Line= 3
      3781823.43     10583520.65      3781324.29      10583472.9
      3779787.84     10583972.03
#Sta/Elev= 30
  3844.4  351.37  3988.9   339.1  4029.1  337.52  4113.1  340.26  4150.6  338.45
  4179.7  332.23    4230  328.34  4378.1  328.18  4425.6  327.55  4578.3  325.86
    4946  326.78  4960.6     327    4967   322.1  4972.3  326.79  4989.1  319.18
  4991.9  318.68  4995.1  319.18    4999   321.5  5004.2  319.62  5030.9  325.23
  5036.2  323.41  5044.7   325.8  5062.9  326.56  5126.8  324.35  5212.8  325.76
  5412.7  326.95  5570.4  330.35  5643.3  333.52  5791.2  345.24  5961.3  348.03
#Mann= 8 ,-1 , 0
  3844.4     .16       0  4150.6     .12       0  4378.1     .16       0
  4425.6     .12       0    4946     .16       0  4989.1     .07       0
  4995.1     .16       0  5212.8     .05       0
Bank Sta=4972.3,5030.9
XS Rating Curve= 0 ,0
Exp/Cntr=0.3,0.1

Type RM Length L Ch R = 1 ,101965  ,924,924,924
BEGIN DESCRIPTION:
BOX CREEK 137.0
END DESCRIPTION:
XS GIS Cut Line= 3
      3781551.87     10582589.54      3780692.46     10582995.81
      3779734.38     10583839.33
#Sta/Elev= 30
  3946.6  363.37  4009.4  362.47  4144.8  360.68  4360.7  353.85  4643.4  336.38
  4707.7  332.69  4767.6  326.48  4844.2  324.91  4966.4  325.77  4973.1  323.78
  4980.7  317.71  4984.3  316.47  4987.1  315.97  4990.3  316.47  5001.6  316.75
  5003.7  317.98  5008.2  320.63  5015.8  320.58  5022.4  325.39  5107.8  325.58
  5150.5  324.07  5320.3  325.25  5426.6   323.6  5688.5  325.05  5731.1  326.35
  5780.5  331.77  5922.8  340.79  5993.5  343.84    6142  344.82  6173.7   343.8
#Mann= 6 ,-1 , 0
  3946.6     .16       0  4009.4     .12       0  4643.4     .16       0
  4984.3     .07       0  4990.3     .16       0  5003.7     .05       0
Bank Sta=4966.4,5022.4
XS Rating Curve= 0 ,0
Exp/Cntr=0.3,0.1

Type RM Length L Ch R = 1 ,101041  ,721,721,721
BEGIN DESCRIPTION:
BOX CREEK 136.0
END DESCRIPTION:
XS GIS Cut Line= 3
      3781349.56     10582560.19      3780149.61     10582660.19
      3779449.58     10583760.23
#Sta/Elev= 30
  3833.8  360.39  4098.6  346.25  4198.2  340.02  4397.3  331.35  4512.8  326.95
  4753.4  322.24  4980.2  324.05  4987.7  321.92  4997.8  315.82  5007.8  316.78
  5017.8  322.52  5057.4  323.02  5166.1  323.06  5175.9  321.93  5181.8  317.96
  5191.2  318.45  5197.1  314.01  5200.9  313.77  5203.6  313.27  5206.9  313.77
  5227.6     315  5248.7  322.57    5385  320.73  5407.2  322.08  5536.9  322.62
  5687.5  326.34  5770.3   331.8    5943  336.28  6094.5  343.65  6341.8   348.6
#Mann= 13 ,-1 , 0
  3833.8     .12       0  4098.6     .16       0  4198.2     .12       0
  4397.3     .16       0  4512.8     .05       0  4753.4     .16       0
  5057.4     .12       0  5166.1     .16       0  5200.9     .07       0
  5206.9     .16       0  5407.2     .05       0  5536.9     .16       0
  5687.5     .05       0
Bank Sta=5166.1,5248.7
XS Rating Curve= 0 ,0
Exp/Cntr=0.3,0.1

Type RM Length L Ch R = 1 ,100320  ,557,557,557
BEGIN DESCRIPTION:
BOX CREEK 135.0
END DESCRIPTION:
XS GIS Cut Line= 3
      3780649.58     10581810.21      3779849.61     10582610.19
      3779449.62     10583010.17
#Sta/Elev= 30
  3856.6  350.48  3927.3   346.8  4026.3  338.69  4054.6   337.7  4082.8  334.78
    4097  331.34    4196  327.24  4262.9  325.86  4563.7  320.84  4606.1  320.56
    4691  322.22    4796  321.94  4917.2  320.57  4931.4  321.77  4973.8   322.4
  4984.4  320.05  4991.5  320.05  4999.1  314.11  5001.8  313.61  5005.1  314.11
  5016.2  321.37  5030.4  321.71  5044.5  320.13  5062.5  320.31  5086.9  321.57
  5200.1  320.87  5256.6   322.1  5383.9     331  5412.2  334.49  5553.6  340.52
#Mann= 6 ,-1 , 0
  3856.6     .12       0  4262.9     .05       0    4796     .16       0
  4999.1     .07       0  5005.1     .16       0  5062.5     .05       0
Bank Sta=4973.8,5030.4
XS Rating Curve= 0 ,0
Exp/Cntr=0.3,0.1

Type RM Length L Ch R = 1 ,99763   ,567,567,567
BEGIN DESCRIPTION:
BOX CREEK 134.0
END DESCRIPTION:
XS GIS Cut Line= 3
      3780749.63     10581610.18      3779649.61     10582160.19
      3778949.61     10583260.19
#Sta/Elev= 30
  3765.1  354.18  3790.6  353.68  3935.6  348.84  4069.8  339.69  4153.6  331.28
  4235.1  327.35  4338.1   323.5  4660.5  320.28  4958.6  321.18  4972.6  319.83
  4989.2  312.54  4991.9  312.04  4995.2  312.54  5002.6  315.97  5008.5  316.05
  5017.8  320.91  5023.7  316.38    5039  317.55  5044.9  316.06  5054.2  318.23
  5066.1  316.96  5075.4  320.81  5090.6  320.74  5226.9  321.63  5414.9  319.55
  5618.1  330.38  5675.7  331.76  5763.7  340.04  5821.3  342.76  6298.8  346.54
#Mann= 7 ,-1 , 0
  3765.1     .16       0  3790.6     .12       0  4235.1     .05       0
  4660.5     .16       0  4989.2     .07       0  4995.2     .16       0
  5090.6     .05       0
Bank Sta=4958.6,5017.8
XS Rating Curve= 0 ,0
Exp/Cntr=0.3,0.1

Type RM Length L Ch R = 1 ,99196   ,561,561,561
BEGIN DESCRIPTION:
BOX CREEK 133.0
END DESCRIPTION:
XS GIS Cut Line= 3
      3780199.59     10581160.21      3779399.61     10581960.19
      3778799.63     10582610.17
#Sta/Elev= 30
  3872.7  344.97  3929.2  335.26  4050.1  329.57  4141.4  325.09  4202.9  325.36
    4242  323.81  4749.5  318.11  4876.8  320.62  4975.8  320.22  4989.9  310.67
  4997.5   310.3  5000.3   309.8  5003.5   310.3  5005.1   310.3  5011.1  311.96
  5017.9  318.53  5032.1  320.16  5105.1  319.15  5159.7  320.14  5230.6   318.8
  5237.4  317.39  5244.7  318.95  5273.1  318.29  5301.5  320.33  5506.7  318.65
  5626.9  321.17  5747.2  328.75  5872.8   342.5  5878.6  342.52  5888.6  342.96
#Mann= 10 ,-1 , 0
  3872.7     .16       0  4050.1     .05       0  4202.9     .16       0
    4242     .05       0  4997.5     .03       0  5003.5     .05       0
  5005.1     .16       0  5105.1     .05       0  5872.8     .08       0
  5878.6     .05       0
Bank Sta=4975.8,5032.1
XS Rating Curve= 0 ,0
Exp/Cntr=0.3,0.1

Type RM Length L Ch R = 1 ,98635   ,486,486,486
BEGIN DESCRIPTION:
BOX CREEK 132.0
END DESCRIPTION:
XS GIS Cut Line= 3
      3779949.58     10581060.22      3779149.61     10581810.19
      3778449.65     10582060.17
#Sta/Elev= 30
  3926.4  348.13  3990.1   333.5  4011.1  331.74  4018.4  328.94  4025.3  329.77
  4032.6  327.26  4060.9  325.19  4195.2   319.9  4308.6  321.03  4549.9  317.87
  4618.7   317.2  4973.4  318.29  4980.7  316.93  4987.5  312.16  4998.7  311.74
  5001.4  311.24  5004.7  311.74    5009  316.25  5036.3  319.07  5044.2  319.43
  5079.6  318.71  5142.7  318.36  5181.7  320.57  5243.3  318.55  5268.3  319.74
  5352.1  322.94  5437.1  331.45  5602.2  334.92  5741.2  341.87  5766.2  342.59
#Mann= 11 ,-1 , 0
  3926.4     .16       0  4025.3     .05       0  4549.9     .16       0
  4618.7     .12       0  4998.7     .07       0  5004.7     .12       0
  5036.3     .05       0  5079.6     .12       0  5142.7     .05       0
  5268.3     .16       0  5741.2     .05       0
Bank Sta=4973.4,5044.2
XS Rating Curve= 0 ,0
Exp/Cntr=0.3,0.1

Type RM Length L Ch R = 1 ,98149   ,587,587,587
BEGIN DESCRIPTION:
BOX CREEK 131.0
END DESCRIPTION:
XS GIS Cut Line= 3
      3779849.62     10580410.18      3778899.61     10581410.19
      3778399.63     10581910.17
#Sta/Elev= 30
  3617.8  366.28  3663.7  364.26  3730.9  361.96  3773.3  356.23  3851.4  335.93
  3937.2  322.74  4070.6  318.15  4315.2  315.51  4464.9  316.34  4473.5  318.57
  4494.9  318.83  4530.2  314.97  4558.9   315.4  4761.6  316.16  4892.1  317.24
  4913.7  317.92  4961.7  318.19    4969  316.14  4975.9  318.35  4990.7  308.92
  4993.4  308.42  4996.7  308.92  5023.3  315.85  5039.5  317.93  5364.8  315.29
  5462.6  318.15  5591.1  327.93  5647.7   337.3  5676.4  339.88  5704.2  341.94
#Mann= 14 ,-1 , 0
  3617.8     .05       0  3663.7     .16       0  3937.2     .05       0
  4315.2     .16       0  4464.9     .05       0  4558.9     .12       0
  4761.6     .16       0  4892.1     .12       0  4913.7     .16       0
  4990.7     .07       0  4996.7     .16       0  5023.3     .05       0
  5462.6     .16       0  5676.4     .05       0
Bank Sta=4975.9,5039.5
XS Rating Curve= 0 ,0
Exp/Cntr=0.3,0.1

Type RM Length L Ch R = 1 ,97562   ,488,488,488
BEGIN DESCRIPTION:
BOX CREEK 130.0
END DESCRIPTION:
XS GIS Cut Line= 3
       3779549.6      10580210.2      3778749.61     10581010.19
       3778349.6     10581810.21
#Sta/Elev= 30
  3847.9  366.86  3856.4  366.33  3904.5  359.06  3975.2  339.72  4032.7   330.6
  4088.3  326.26    4159  323.52  4215.6  322.18  4328.7   323.1  4371.1  320.76
  4399.4  321.77  4475.6  316.74    4555  314.21  4682.3  313.11    4982  316.21
  4987.6  314.85  4993.2  309.57  4998.6  307.15  5001.4  306.65  5004.6  307.15
  5015.6  313.53    5024  315.95  5026.5  315.91    5337  316.36  5359.4  313.84
  5434.9  315.66  5641.7  314.52  5747.9  316.95  5769.7  319.38  5873.7  336.27
#Mann= 8 ,-1 , 0
  3847.9     .05       0  3856.4     .16       0  4032.7     .05       0
  4475.6     .12       0  4998.6     .07       0  5004.6     .12       0
  5026.5     .05       0  5769.7     .16       0
Bank Sta=4982,5024
XS Rating Curve= 0 ,0
Exp/Cntr=0.3,0.1

Type RM Length L Ch R = 1 ,97074   ,581,581,581
BEGIN DESCRIPTION:
BOX CREEK 129.0
END DESCRIPTION:
XS GIS Cut Line= 3
      3779349.64     10579810.16      3778599.61     10580610.19
      3777749.64     10581860.15
#Sta/Elev= 30
  3862.3  370.35  3910.8  367.64  4003.8  354.69  4069.4  342.32  4168.3  331.57
  4407.2  318.39  4428.2  320.97  4498.8  316.75  4626.5  313.14  4902.5  314.22
  4916.7  307.24  4937.7  309.78    4945  306.57  4951.8  312.25  4955.5  306.39
  4987.4  307.71  4995.2  310.44  5014.3  305.92    5017  305.42  5020.3  305.92
  5044.3  314.33  5162.2  313.69  5297.5  312.73  5361.5  316.41  5484.3  317.31
    5592  313.55    5867  313.68  6023.1  316.17  6219.2  338.42  6470.5  343.06
#Mann= 10 ,-1 , 0
  3862.3     .05       0  3910.8     .12       0  4069.4     .16       0
  4168.3     .05       0  4498.8     .12       0  5014.3     .07       0
  5020.3     .12       0  5162.2     .05       0    5867     .12       0
  6219.2     .05       0
Bank Sta=4902.5,5044.3
XS Rating Curve= 0 ,0
Exp/Cntr=0.3,0.1

Type RM Length L Ch R = 1 ,96493   ,698,698,698
BEGIN DESCRIPTION:
BOX CREEK 128.0
END DESCRIPTION:
XS GIS Cut Line= 3
       3778949.6      10579760.2      3778449.61     10580160.19
      3777749.62     10581710.16
#Sta/Elev= 30
  4359.2  372.27  4401.6   367.9  4430.4  356.25  4530.3  333.65  4608.1  322.12
  4643.3  323.34  4657.7  320.01  4720.6  316.83  4878.6  311.09  4957.1  313.79
  4963.5  310.35  4971.5  313.67  4977.9  306.09  4993.3  305.81    4996  305.31
  4999.3  305.81  5013.8  306.72  5021.4  313.37  5307.6   312.9  5416.5   312.8
  5428.8  314.76  5446.4  312.48  5559.1  312.05  6211.3  313.15    6244  313.22
  6349.8     316  6419.5  323.34    6490  335.72  6530.6  339.59  6700.2  342.65
#Mann= 11 ,-1 , 0
  4359.2     .12       0  4530.3     .05       0  4720.6     .12       0
  4993.3     .07       0  4999.3     .12       0  5307.6     .05       0
  6211.3     .12       0    6244     .16       0  6349.8     .12       0
  6419.5     .16       0  6530.6     .05       0
Bank Sta=4971.5,5021.4
XS Rating Curve= 0 ,0
Exp/Cntr=0.3,0.1

Type RM Length L Ch R = 1 ,95795   ,574,574,574
BEGIN DESCRIPTION:
BOX CREEK 127.0
END DESCRIPTION:
XS GIS Cut Line= 3
       3778399.6     10579110.22      3778099.61     10579810.19
      3777549.61     10581210.19
#Sta/Elev= 30
  4248.6  375.14  4295.7  370.91  4357.4  363.81  4368.2  359.07  4409.9  351.37
  4538.7   337.1  4544.1   331.3  4562.3   332.2  4585.8  326.01  4614.8  327.26
  4643.9  322.61  4731.5  319.56  4879.8  314.21  4977.5  312.28  5016.7  304.94
  5019.4  304.44  5022.7  304.94  5031.6   312.7  5195.6  311.36  5512.9  311.53
  5537.4   308.9  5630.3  311.29  5903.1  312.01  5957.3  316.64  5998.6  312.43
  6245.7  313.34  6320.9  318.25  6428.4  333.46  6476.4  337.44  6514.3  338.19
#Mann= 10 ,-1 , 0
  4248.6     .12       0  4295.7     .16       0  4731.5     .05       0
  4879.8     .12       0  5016.7     .07       0  5022.7     .12       0
  5195.6     .05       0  5537.4     .12       0  5630.3     .05       0
  6476.4     .16       0
Bank Sta=4977.5,5031.6
XS Rating Curve= 0 ,0
Exp/Cntr=0.3,0.1

Type RM Length L Ch R = 1 ,95221   ,639,639,639
BEGIN DESCRIPTION:
BOX CREEK 126.0
END DESCRIPTION:
XS GIS Cut Line= 3
       3778349.6      10579060.2      3777749.61     10579610.19
       3777499.6     10581160.23
#Sta/Elev= 30
  4175.3  376.24  4267.5  366.94  4310.4  358.16  4359.4  349.95  4445.5  341.51
  4449.4  341.09  4584.8  327.53  4588.5  327.11  4635.6  320.07  4724.1  313.62
  4727.5  313.32  4863.5  310.18  4953.8  311.23  4961.2  311.03    4968  307.23
  4975.4  308.08  4982.1  303.67  4996.4  303.62  4999.1  303.12  5002.4  303.62
  5009.5  309.94  5022.7  311.12  5455.2  310.85  5475.4   308.1  5614.2  310.98
  5971.8  314.45  6335.4  314.87  6387.1  318.08  6498.5  336.26  6559.3  338.75
#Mann= 12 ,-1 , 0
  4175.3     .16       0  4310.4      .1       0  4445.5     .16       0
  4449.4      .1       0  4584.8     .12       0  4588.5     .07       0
  4724.1     .05       0  4727.5      .1       0  4863.5     .12       0
  4996.4     .07       0  5002.4     .12       0  5614.2     .05       0
Bank Sta=4953.8,5022.7
XS Rating Curve= 0 ,0
Exp/Cntr=0.3,0.1

Type RM Length L Ch R = 1 ,94582   ,1081,1081,1081
BEGIN DESCRIPTION:
BOX CREEK 125.0
END DESCRIPTION:
XS GIS Cut Line= 3
      3777994.45     10578960.16      3777304.32     10579702.38
      3776288.71     10580123.38
#Sta/Elev= 30
  4193.2  346.32  4396.4   326.3  4428.6  324.12  4451.6  319.74  4529.3  314.29
  4599.4  312.56  4687.2   310.7  4699.4  309.93  4934.3  310.06  4953.8  310.21
  4960.7  310.09    4968   305.1  4979.2   303.4  4981.9   302.9  4985.2   303.4
  5003.2  303.95  5010.5  309.41  5017.4  309.78  5255.1  309.65  5277.5  304.28
  5309.2  308.97  5386.3  307.88  5495.1  307.96    5667  307.48  5731.1  307.87
  5821.4  317.07  5906.1  328.42  5925.7  331.61  6044.8  337.18  6306.1  337.54
#Mann= 16 ,-1 , 0
  4193.2     .05       0  4396.4     .12       0  4428.6     .07       0
  4599.4     .12       0  4687.2     .05       0  4699.4     .07       0
  4934.3     .12       0  4979.2     .07       0  4985.2     .12       0
  5277.5     .16       0  5386.3     .12       0  5495.1     .05       0
    5667     .16       0  5821.4     .12       0  5906.1     .16       0
  5925.7     .05       0
Bank Sta=4953.8,5017.4
XS Rating Curve= 0 ,0
Exp/Cntr=0.3,0.1

Type RM Length L Ch R = 1 ,93501   ,1111,1111,1111
BEGIN DESCRIPTION:
BOX CREEK 124.0
END DESCRIPTION:
XS GIS Cut Line= 3
      3777775.17     10578768.92      3777030.93     10579383.61
      3776436.59     10579759.51
#Sta/Elev= 30
  3971.4  335.77  3978.1  335.14  3997.5  334.13  4018.3  329.61  4040.5   327.5
  4072.1  326.84  4246.3  313.83  4513.7  307.79  4640.4  307.64  4808.1  308.52
  4905.3  308.07  4958.5  308.38  4978.3  308.44  4985.6  308.32  4996.5  302.02
  4999.3  301.52  5002.5  302.02  5008.9  302.77  5014.8  307.05  5021.1  308.51
  5028.2  308.47  5131.5  306.65  5304.5  305.65  5406.5  308.01  5458.2  314.41
  5485.3  319.43  5521.7  329.56  5542.9  332.53  5609.9   336.5  5639.9  335.96
#Mann= 13 ,-1 , 0
  3971.4     .05       0  3978.1     .12       0  4072.1     .07       0
  4513.7     .12       0  4640.4     .07       0  4808.1     .12       0
  4905.3     .16       0  4958.5     .12       0  4996.5     .07       0
  5002.5     .12       0  5028.2     .16       0  5131.5     .05       0
  5304.5     .12       0
Bank Sta=4978.3,5021.1
XS Rating Curve= 0 ,0
Exp/Cntr=0.3,0.1

Type RM Length L Ch R = 1 ,92390   ,665,665,665
BEGIN DESCRIPTION:
BOX CREEK 123.0
END DESCRIPTION:
XS GIS Cut Line= 3
        3777671.     10578415.88      3776916.63     10578939.11
      3776266.38     10579500.46
#Sta/Elev= 30
  4042.7  331.38  4233.8  320.87  4320.2  317.27  4396.4  316.09  4408.5  315.73
  4514.1  311.08  4660.2  308.39  4773.5  307.05  4809.3  305.46  4859.8  307.18
  4976.3  307.09    4981  307.34  4987.6  307.16  4995.3  301.86  4998.9  300.57
  5001.6  300.07  5004.9  300.57  5016.1  302.34  5022.9  307.31  5196.7     307
  5434.1  305.11    5512     306  5590.9  304.43  5623.8  305.71  5695.2  314.68
  5724.8  320.56  5753.3  329.45  5767.5  330.83  5789.1   333.1  5819.8  333.29
#Mann= 11 ,-1 , 0
  4042.7     .07       0  4396.4     .05       0  4408.5     .07       0
  4660.2     .12       0  4976.3     .16       0  4998.9     .07       0
  5004.9     .16       0  5196.7     .05       0  5623.8     .12       0
  5695.2     .16       0  5767.5     .12       0
Bank Sta=4981,5022.9
XS Rating Curve= 0 ,0
Exp/Cntr=0.3,0.1

Type RM Length L Ch R = 1 ,91725   ,1305,1305,1305
BEGIN DESCRIPTION:
BOX CREEK 122.0
END DESCRIPTION:
XS GIS Cut Line= 4
      3777373.82     10578050.14      3776789.64       10578614.
      3776670.26     10578801.96      3776045.42     10579279.48
#Sta/Elev= 30
  4010.3  336.28    4070  329.29  4084.1  326.47  4126.5  322.67    4176  318.61
  4254.9  314.61  4262.3  314.49  4397.7  310.46  4398.6  310.41  4550.8  309.54
  4673.9  306.21  4985.1  306.19  4994.5  303.09  4997.4  299.26  5000.1  298.76
  5003.4  299.26  5007.2  301.52  5015.6  302.54  5021.6  306.46  5063.7  305.82
  5113.9  305.55  5574.5  304.62  5593.4  305.06    5637  310.78  5649.8   314.1
  5664.1  315.15  5693.2  323.57  5743.1  331.47  5800.6  332.97  5831.3  333.31
#Mann= 13 ,-1 , 0
  4010.3     .07       0  4126.5     .05       0  4254.9     .12       0
  4262.3     .05       0  4397.7     .12       0  4398.6     .05       0
  4673.9     .12       0  4997.4     .07       0  5003.4     .12       0
  5063.7     .16       0  5113.9     .05       0  5574.5     .12       0
  5800.6     .16       0
Bank Sta=4985.1,5021.6
XS Rating Curve= 0 ,0
Exp/Cntr=0.3,0.1

Type RM Length L Ch R = 1 ,90420   ,724,724,724
BEGIN DESCRIPTION:
BOX CREEK 121.0
END DESCRIPTION:
XS GIS Cut Line= 3
      3776799.57     10578210.22      3776399.61     10578510.19
      3775799.64     10578410.19
#Sta/Elev= 30
  4483.2  329.83  4511.3   328.4  4540.4  321.51  4561.3  320.64  4590.4  313.56
  4625.9  310.93  4676.8  304.43  4733.2  304.23  4746.7  302.75  4775.9   304.6
  4870.2  304.58  4975.9  304.57    4980  301.13  4989.9  299.26  4990.3  299.08
    4993  298.58  4996.3  299.08    5011  304.48    5170  304.36  5185.9  304.11
  5206.2  306.45  5226.5  304.27  5348.1  303.37    5369  300.91  5419.1  300.51
  5469.8  309.06  5485.4  313.22  5520.5  323.02  5558.5  329.01  5591.4  331.64
#Mann= 9 ,-1 , 0
  4483.2     .12       0  4676.8     .16       0  4870.2     .12       0
  4989.9     .16       0  4990.3     .07       0  4996.3     .16       0
    5170     .05       0    5369     .16       0  5485.4     .12       0
Bank Sta=4975.9,5011
XS Rating Curve= 0 ,0
Exp/Cntr=0.3,0.1

Type RM Length L Ch R = 1 ,89696   ,602,602,602
BEGIN DESCRIPTION:
BOX CREEK 120.0
END DESCRIPTION:
XS GIS Cut Line= 3
      3776899.65     10577860.17      3776349.61     10578110.19
      3775799.65     10578360.17
#Sta/Elev= 30
  4412.2  344.81  4444.1  342.05  4518.8   327.2    4610  315.65  4616.6  312.87
    4622  313.84  4668.2  307.99  4737.4  303.65  4904.4  302.49  4917.5  300.86
  4972.5     304    4979  302.16  4984.5  303.01  4994.4  298.96  5002.1  301.94
  5004.6  296.22  5007.4  295.72  5010.6  296.22  5013.6  303.56  5235.6  303.31
  5373.7  301.68  5393.2   301.5  5400.9  299.44  5419.2  300.22  5422.8  301.65
  5444.8  302.12  5500.8  310.51  5537.1  315.86  5583.2  326.07  5620.5  329.83
#Mann= 7 ,-1 , 0
  4412.2     .12       0  5004.6     .07       0  5010.6     .12       0
  5235.6     .16       0  5373.7     .12       0  5419.2     .16       0
  5500.8     .12       0
Bank Sta=4972.5,5013.6
XS Rating Curve= 0 ,0
Exp/Cntr=0.3,0.1

Type RM Length L Ch R = 1 ,89094   ,712,712,712
BEGIN DESCRIPTION:
BOX CREEK 119.0
END DESCRIPTION:
XS GIS Cut Line= 3
      3776749.63     10577660.18      3775949.61     10577960.19
      3775749.63     10578310.15
#Sta/Elev= 30
  4118.1  345.41  4150.2  341.77  4243.6  320.02    4249  321.03  4273.9  314.77
  4342.4  305.64  4389.6  300.96    4455  302.02  4737.6  303.47  4748.2  303.26
  4761.6  296.29  4791.9   298.4  4808.4  295.94  4811.2  295.44  4814.4  295.94
  4841.7  303.45    4855   298.6  4887.1   303.5  4974.6  303.26  4980.4  302.89
  5017.9  296.34  5066.8     306  5098.5  307.11  5141.7  312.85  5147.4  318.27
  5156.8  316.24    5169     322  5184.9  323.89  5343.3  330.63  5375.6  331.43
#Mann= 6 ,-1 , 0
  4118.1     .12       0    4455     .16       0  4808.4     .07       0
  4814.4     .16       0  4974.6     .12       0  5343.3     .05       0
Bank Sta=4980.4,5066.8
XS Rating Curve= 0 ,0
Exp/Cntr=0.3,0.1

Type RM Length L Ch R = 1 ,88382   ,617,617,617
BEGIN DESCRIPTION:
BOX CREEK 118.0
END DESCRIPTION:
XS GIS Cut Line= 3
      3776976.12     10576969.73      3776003.91     10577421.11
      3775553.59     10577732.87
#Sta/Elev= 30
  3824.7  337.66  3911.7  334.89  3964.2  327.65  4019.3  322.04  4026.2  320.05
  4107.5  312.74  4169.1  308.61  4197.6   309.1  4214.9  307.34  4228.8  308.36
  4299.2     305  4386.3  301.81  4658.8  300.16  4992.3  302.94  4999.1   296.8
  5004.2  295.06  5006.9  294.56  5010.2  295.06  5013.3  295.93    5022   303.9
  5049.1  309.32  5078.8  312.08  5084.9  313.98  5108.5  315.11  5114.6   317.1
  5150.4  321.01  5171.4  325.83  5179.5  325.89    5243  330.07  5444.3  331.51
#Mann= 5 ,-1 , 0
  3824.7     .16       0  4299.2     .12       0  5004.2     .07       0
  5010.2     .12       0  5179.5     .05       0
Bank Sta=4992.3,5022
XS Rating Curve= 0 ,0
Exp/Cntr=0.3,0.1

Type RM Length L Ch R = 1 ,87765   ,745,745,745
BEGIN DESCRIPTION:
BOX CREEK 117.0
END DESCRIPTION:
XS GIS Cut Line= 3
      3776170.56     10576636.42      3775837.25     10577150.28
      3775198.33     10577560.01
#Sta/Elev= 30
  4272.3  335.85  4304.1  335.57  4334.4  331.77  4376.6  331.31    4428  323.65
  4449.1  325.77  4485.4  321.45  4548.9  307.67  4630.4  297.92  4890.9  302.21
    4977  301.45  4990.7   300.8  4996.9  294.29  4999.7  293.79  5002.9  294.29
  5005.9  295.81  5012.7  294.45  5021.1  301.67    5027   301.8  5130.1  302.34
  5187.6  309.45  5221.4  316.97    5251  324.39  5281.4   324.5  5301.1  327.63
  5317.8  325.98  5466.4  327.73  5472.6  327.92  5610.6  328.56  5643.8  327.43
#Mann= 9 ,-1 , 0
  4272.3     .16       0  4548.9     .12       0  4996.9     .07       0
  5002.9     .12       0  5221.4     .16       0  5301.1     .05       0
  5466.4     .16       0  5472.6     .05       0  5610.6     .16       0
Bank Sta=4977,5027
XS Rating Curve= 0 ,0
Exp/Cntr=0.3,0.1

Type RM Length L Ch R = 1 ,87020   ,559,559,559
BEGIN DESCRIPTION:
BOX CREEK 116.0
END DESCRIPTION:
XS GIS Cut Line= 3
       3775958.8     10576551.36      3775602.94     10576811.75
      3774874.16     10577019.97
#Sta/Elev= 30
  4493.8  336.12    4529  334.07  4564.5  329.56  4591.9  324.01    4600  320.81
  4635.5  311.82  4728.2     301  4836.3  298.88  4857.1  300.02  4984.3  300.09
  4990.2   293.3  4997.6  293.14  5000.4  292.64  5003.6  293.14    5011  300.45
  5225.5  300.33  5260.6   301.1  5314.6  307.46  5348.4  312.78  5354.2  315.92
  5364.6   316.8    5375  319.96  5384.9  321.03    5416  325.93  5488.9  329.35
  5497.6   329.1  5605.8  330.41  5624.6  329.65  5639.6  326.84  5692.7   328.8
#Mann= 7 ,-1 , 0
  4493.8     .16       0  4997.6     .07       0  5003.6     .16       0
  5225.5     .12       0  5384.9     .16       0  5488.9     .05       0
  5497.6     .16       0
Bank Sta=4984.3,5011
XS Rating Curve= 0 ,0
Exp/Cntr=0.3,0.1

Type RM Length L Ch R = 1 ,86461   ,646,646,646
BEGIN DESCRIPTION:
BOX CREEK 115.0
END DESCRIPTION:
XS GIS Cut Line= 3
      3775849.61     10576310.19      3775449.61     10576360.19
      3775099.64     10576560.17
#Sta/Elev= 30
    4635  328.52  4665.2  328.02  4677.8  329.03  4758.5  324.58  4846.6  313.93
  4876.9  312.46  4885.8  310.64  4914.7  307.66  4919.7  308.24  4967.6  301.57
  4977.7  295.23  4987.7  292.55  4997.3  292.17  5000.1  291.67  5003.3  292.17
  5007.9  298.85  5222.4  298.97  5234.6  299.86    5280  297.63  5287.9  300.11
  5293.7  299.95    5303  302.21  5309.5  305.99  5331.1  307.49  5337.6  310.52
  5352.7   312.3  5360.6   315.5  5374.3  317.29  5383.6  320.39  5441.2  325.08
#Mann= 4 ,-1 , 0
    4635     .16       0  4885.8     .12       0  4997.3     .07       0
  5003.3     .12       0
Bank Sta=4967.6,5007.9
XS Rating Curve= 0 ,0
Exp/Cntr=0.3,0.1

Type RM Length L Ch R = 1 ,85815   ,619,619,619
BEGIN DESCRIPTION:
BOX CREEK 114.0
END DESCRIPTION:
XS GIS Cut Line= 3
      3776049.57     10575660.21      3775249.61     10576060.19
      3774849.61     10576110.19
#Sta/Elev= 30
  4183.2  343.72  4272.6  333.23  4325.7  319.69  4331.3  321.14  4406.8  308.04
  4510.2  301.28    4527  297.79  4540.9  301.06  4818.5   297.3  4957.4  299.05
  4979.8  298.03  4988.1  293.18  5002.1  291.87  5018.9  299.08  5055.2  298.17
  5069.2  295.59  5074.8  291.57  5094.7  291.17  5097.5  290.67  5100.7  291.17
  5107.8  294.08    5128  293.26  5148.1  298.88  5168.3  301.48  5218.7  297.27
  5248.9  303.92  5276.6  303.05  5319.5   308.8  5369.8  322.16  5480.7  331.57
#Mann= 4 ,-1 , 0
  4183.2     .16       0  4818.5     .12       0  5094.7     .07       0
  5100.7     .12       0
Bank Sta=5055.2,5148.1
XS Rating Curve= 0 ,0
Exp/Cntr=0.3,0.1

Type RM Length L Ch R = 1 ,85196   ,557,557,557
BEGIN DESCRIPTION:
BOX CREEK 113.0
END DESCRIPTION:
XS GIS Cut Line= 3
      3775899.63     10575410.18      3775099.61     10575660.19
       3774749.6      10575860.2
#Sta/Elev= 30
  4189.9  338.94  4246.5  329.62  4263.3  327.53  4276.4  322.45  4303.6  318.08
  4315.6  313.58    4379  303.72  4451.8  298.27  4561.4  298.13  4567.1  297.67
  4573.9  292.67  4582.2  296.12  4853.5  297.06  4974.1  298.45  5008.8  290.44
  5011.6  289.94  5014.8  290.44  5017.6  294.73  5028.1  298.58  5073.4  307.72
  5079.2  306.93    5095  312.54  5100.8   310.7  5116.6  316.94  5122.4  316.02
  5138.2  321.11  5159.8  321.26  5197.2  326.25  5246.9  329.35  5431.2  330.66
#Mann= 7 ,-1 , 0
  4189.9     .05       0  4246.5     .16       0  4561.4     .12       0
  4582.2     .16       0  4853.5     .12       0  5008.8     .07       0
  5014.8     .12       0
Bank Sta=4974.1,5028.1
XS Rating Curve= 0 ,0
Exp/Cntr=0.3,0.1

Type RM Length L Ch R = 1 ,84639   ,389,389,389
BEGIN DESCRIPTION:
BOX CREEK 112.0
END DESCRIPTION:
XS GIS Cut Line= 3
      3775899.63     10575360.19      3775349.61     10575210.19
      3774949.63     10575310.18
#Sta/Elev= 30
  4433.6  343.25  4475.1  339.88  4511.3  331.99  4547.6  325.17  4564.9   320.8
  4578.7  315.09  4589.1  314.67  4609.8  308.09  4692.8   298.6    4786   295.2
  4906.7  296.98  4941.5  297.25  4986.4  295.03  4993.3  289.73  4996.3  289.06
  4998.1  288.65  5000.9  288.15  5004.1  288.65  5009.7  291.47    5014  295.04
  5021.7   297.2  5086.2  295.51  5109.4  298.31  5150.6  307.19  5158.3  310.56
  5178.9  315.23  5199.6  317.92  5274.3  320.72    5364  321.12    5416  322.16
#Mann= 8 ,-1 , 0
  4433.6     .05       0  4511.3     .16       0  4906.7     .12       0
  4996.3     .16       0  4998.1     .07       0  5004.1     .16       0
  5009.7     .12       0    5364     .05       0
Bank Sta=4986.4,5021.7
XS Rating Curve= 0 ,0
Exp/Cntr=0.3,0.1

Type RM Length L Ch R = 1 ,84250   ,309,309,309
BEGIN DESCRIPTION:
BOX CREEK 111.0
END DESCRIPTION:
XS GIS Cut Line= 2
       3776300.8     10574711.04      3774868.47     10574919.38
#Sta/Elev= 30
  3948.5  330.79  3976.2  327.16  3981.2  327.48  4010.3  324.33    4071  320.52
  4161.9  310.46  4206.2  307.68  4256.6  304.97  4307.4  300.93  4326.7   301.1
    4364  298.96  4399.8   298.4  4434.8  296.94  4545.9  295.36  4608.9  295.72
  4672.1  295.01  4910.4  295.87  4970.3   297.1  4980.4  296.41  4990.5  294.32
  5000.6  288.63  5007.8  288.51  5010.5  288.01  5013.8  288.51  5017.6  295.15
    5054   298.9  5101.7  303.75  5222.9  308.21    5298  309.15  5395.9  308.77
#Mann= 9 ,-1 , 0
  3948.5     .07       0  4206.2     .12       0  4307.4     .16       0
  4399.8     .12       0  4608.9     .05       0  4910.4     .12       0
  5007.8     .07       0  5013.8     .12       0    5054     .05       0
Bank Sta=4980.4,5017.6
XS Rating Curve= 0 ,0
Exp/Cntr=0.3,0.1

Type RM Length L Ch R = 1 ,83941   ,1090,1090,1090
BEGIN DESCRIPTION:
BOX CREEK 110.0
END DESCRIPTION:
XS GIS Cut Line= 3
      3775992.81       10574280.      3775419.91     10574550.83
       3774684.2     10574720.87
#Sta/Elev= 30
  4273.7  339.99  4352.6  333.22  4358.1  330.94  4387.9  326.73  4398.1  322.96
  4417.4  319.34  4426.4  315.81  4465.3  308.79  4487.4  307.37  4494.7  304.74
  4568.5  296.21    4614  293.41  4664.5  294.59  4969.1  296.28  4979.5  295.67
  4997.1  289.56  4999.8  289.06  5003.1  289.56  5010.3  294.76  5015.5  296.15
  5184.8  294.93  5287.5   301.3  5492.7  304.01    5501  302.34  5506.1  304.08
  5513.3   302.6  5523.5  304.04  5554.3  302.56  5603.4  305.51  5662.5  309.44
#Mann= 7 ,-1 , 0
  4273.7     .07       0  4417.4     .16       0  4664.5     .05       0
  4969.1     .12       0  4997.1     .07       0  5003.1     .12       0
  5603.4     .16       0
Bank Sta=4979.5,5015.5
XS Rating Curve= 0 ,0
Exp/Cntr=0.3,0.1

Type RM Length L Ch R = 1 ,82851   ,550,550,550
BEGIN DESCRIPTION:
BOX CREEK 109.0
END DESCRIPTION:
XS GIS Cut Line= 3
      3776099.56     10574110.19      3774849.61     10574060.19
      3774349.58      10574260.2
#Sta/Elev= 30
  3719.6  338.42  3725.9  338.34  3789.6  337.14  3819.6   330.9  3869.7   328.7
  3919.7   323.2  3929.7  324.03  3979.8  318.34  4009.8  312.58  4052.7   307.2
  4094.9  302.23  4232.4  295.27    4280  293.19  4370.1  294.27  4904.4  293.81
  4973.2  294.39    4980  293.08  4985.4  294.65  4992.1   289.7  4999.9  287.78
  5002.6  287.28  5005.9  287.78  5009.6  289.25    5015  288.45  5024.4  294.43
  5164.4  292.41    5225   300.1  5405.4  314.03  5476.8  321.97  5509.1  323.42
#Mann= 8 ,-1 , 0
  3719.6     .16       0  3725.9     .05       0  4052.7     .16       0
  4232.4     .05       0  4904.4     .12       0  4999.9     .07       0
  5005.9     .12       0  5405.4     .16       0
Bank Sta=4985.4,5024.4
XS Rating Curve= 0 ,0
Exp/Cntr=0.3,0.1

Type RM Length L Ch R = 1 ,82301   ,602,602,602
BEGIN DESCRIPTION:
BOX CREEK 108.0
END DESCRIPTION:
XS GIS Cut Line= 3
      3776149.65     10573760.19      3774599.61     10573710.19
      3774199.57     10574060.22
#Sta/Elev= 30
  3359.6  334.18  3619.8  325.76  3729.8   306.1  3759.8  306.02  3809.9  318.09
  3909.9  317.12    3970  312.17    4040  298.36  4131.9  294.36  4340.1  294.82
  4414.5  292.66  4513.4  292.71  4785.1  292.16  4924.2  293.59  4931.8   289.6
  4966.9  293.39  4974.5  287.27  4981.2  290.43  4985.7  286.51  4988.5  286.01
  4991.7  286.51  4995.4   292.4    5003  286.91  5016.7  286.86  5023.9  293.36
  5038.1  297.57  5066.6  304.65  5109.3  308.01  5340.8  314.89    5442  319.81
#Mann= 8 ,-1 , 0
  3359.6     .16       0  4131.9     .05       0  4414.5     .08       0
  4513.4     .05       0  4785.1     .12       0  4985.7     .07       0
  4991.7     .12       0  5340.8     .16       0
Bank Sta=4340.1,5038.1
XS Rating Curve= 0 ,0
Exp/Cntr=0.3,0.1

Type RM Length L Ch R = 1 ,81699   ,1341,1341,1341
BEGIN DESCRIPTION:
BOX CREEK 107.0
END DESCRIPTION:
XS GIS Cut Line= 3
      3775249.61     10571760.19      3774299.61     10573360.19
      3774049.61     10573860.19
#Sta/Elev= 30
  3095.6  327.49  3183.3   320.1    3497  299.33  3610.7   295.1  3746.4  290.44
  4116.2  290.81  4282.3  291.49  4538.7  293.75  4576.4  291.71  4584.2   288.1
  4597.8  289.16  4607.5  293.45  4613.4  293.54  4687.5  290.72  4862.9  293.56
  4978.7  293.11  4984.1  286.49  4986.9  285.99  4990.1  286.49  4992.7  289.95
  5001.1  286.82  5009.5  289.52  5015.1  287.42  5023.5  293.41  5104.5  291.93
  5216.3  295.07  5277.8  301.09  5291.8  300.86  5300.2  303.42  5515.4  317.87
#Mann= 7 ,-1 , 0
  3095.6     .05       0  3610.7     .12       0  4116.2     .16       0
  4282.3     .05       0  4538.7     .12       0  4984.1     .03       0
  4990.1     .05       0
Bank Sta=4978.7,5023.5
XS Rating Curve= 0 ,0
Exp/Cntr=0.3,0.1

Type RM Length L Ch R = 1 ,80358   ,475,475,475
BEGIN DESCRIPTION:
BOX CREEK 106.0
END DESCRIPTION:
XS GIS Cut Line= 3
       3774716.2     10571503.19      3773757.89     10573100.38
      3773889.83     10574412.84
#Sta/Elev= 30
  3323.2  369.36  3362.8   364.3  3438.6  348.42  3516.4  328.86    3565  319.54
  3609.6  314.26  3712.7  297.79  3755.5  294.29  3835.2  290.48  4004.2  289.19
  4120.9  291.47  4126.7  289.77  4142.2     293  4194.3  288.37  4760.1  291.93
  4964.4  291.34    4980  289.83  4984.4  284.69  4987.1  284.19  4990.4  284.69
  5010.7  287.53  5016.9  291.97  5190.2  290.22  5597.7  291.32  5758.5  294.42
  5838.9  297.82    5859  302.15  6009.8  317.51  6110.3  324.04  6504.9  325.58
#Mann= 7 ,-1 , 0
  3323.2     .12       0  3438.6     .16       0  3609.6     .05       0
  4760.1     .12       0  4984.4     .07       0  4990.4     .12       0
  5190.2     .05       0
Bank Sta=3755.5,5758.5
XS Rating Curve= 0 ,0
Exp/Cntr=0.3,0.1

Type RM Length L Ch R = 1 ,79883   ,983,983,983
BEGIN DESCRIPTION:
BOX CREEK 105.0
END DESCRIPTION:
XS GIS Cut Line= 3
       3774653.7     10571287.91      3773487.05     10572829.55
      3771223.86     10574412.39
#Sta/Elev= 30
  3346.2  364.65  3493.6  356.03  3657.9  336.64  3807.7   307.5  3911.9  297.09
  3997.9  294.14  4107.4  293.77  4454.4  288.73  4975.7  291.12  4991.9  286.18
  5029.1  292.11  5066.8  290.76  5226.8  289.87    5452  290.81  5464.7  286.97
  5532.4  290.06  5694.7  288.46    5700  288.56  6819.4     284  6822.2   283.5
  6825.4     284  7070.5  284.63  7224.4  293.85  7424.1  313.88  7504.4  325.56
  7560.1  339.96  7641.6  352.35  7695.7  353.13  7775.4  354.72  8041.3  358.08
#Mann= 18 ,-1 , 0
  3346.2     .16       0  3911.9     .05       0  3997.9      .1       0
  4454.4     .05       0  4975.7     .12       0  5066.8     .16       0
  5226.8     .05       0    5452     .16       0  5532.4     .05       0
  5694.7     .16       0    5700     .12       0  6819.4     .07       0
  6825.4     .12       0  7070.5     .16       0  7560.1      .1       0
  7641.6     .05       0  7695.7      .1       0  7775.4     .05       0
Bank Sta=4107.4,7224.4
XS Rating Curve= 0 ,0
Exp/Cntr=0.3,0.1

Type RM Length L Ch R = 1 ,78900   ,1024,1024,1024
BEGIN DESCRIPTION:
BOX CREEK 104.0
END DESCRIPTION:
XS GIS Cut Line= 3
      3773806.51     10570968.41      3772841.22     10572836.49
      3771174.54      10574211.5
#Sta/Elev= 30
  3512.4  370.67    3629   365.8  3784.5  322.24  3927.8  299.14  4021.5   293.6
  4205.6  288.41  4268.4  287.67  4683.7  286.65  4882.7  287.73  4966.4   289.3
  5001.8  283.32  5011.5  289.29  5234.2  288.73  5253.3  283.17  5256.1  282.67
  5259.3  283.17  5378.3   296.7  5415.6  301.17  5506.7  316.37  5605.1  322.96
  5753.5  319.89  5832.1  314.61  5931.1  292.93    6004  287.82  6512.7  285.37
  6991.8  287.82  7181.9  303.97  7402.1  351.01  7544.1  344.54  7775.8  356.14
#Mann= 14 ,-1 , 0
  3512.4     .16       0  4021.5     .12       0  4205.6     .05       0
  4268.4     .12       0  4683.7     .05       0  4882.7     .12       0
  5253.3     .07       0  5259.3     .12       0  5378.3     .16       0
  5415.6     .12       0  5753.5     .16       0    6004     .05       0
  6512.7     .12       0  6991.8     .05       0
Bank Sta=3784.5,5605.1
XS Rating Curve= 0 ,0
Exp/Cntr=0.3,0.1

Type RM Length L Ch R = 1 ,77876   ,726,726,726
BEGIN DESCRIPTION:
BOX CREEK 103.0
END DESCRIPTION:
XS GIS Cut Line= 2
      3773723.16     10570864.28      3771167.63     10574010.08
#Sta/Elev= 30
  3023.9  353.81  3194.3  346.92  3200.8  343.08  3272.6  333.47  3279.1  329.17
  3485.2  303.29    3621  296.31  3777.3  295.02  3940.6  293.44  4274.7  304.61
  4480.8  286.45  4977.9  287.98  4997.2  282.96  4999.9  282.46  5003.2  282.96
  5017.6  285.16  5028.5  288.76  5586.3  285.33  5912.2  283.54  6049.4  283.54
  6154.3  284.22  6257.2     289  6464.1  298.42  6478.5  296.48  6569.3  304.89
  6691.1  318.46  6784.7  334.76  6847.7  347.61  6969.1  343.63  7076.9  352.34
#Mann= 12 ,-1 , 0
  3023.9     .16       0  3777.3     .12       0  4997.2     .07       0
  5003.2     .12       0  5017.6     .05       0  5586.3     .12       0
  5912.2     .05       0  6049.4     .07       0  6154.3     .12       0
  6257.2     .05       0  6569.3     .12       0  6784.7     .16       0
Bank Sta=4977.9,5028.5
XS Rating Curve= 0 ,0
Exp/Cntr=0.3,0.1

Type RM Length L Ch R = 1 ,77150   ,677,677,677
BEGIN DESCRIPTION:
BOX CREEK 102.0
END DESCRIPTION:
XS GIS Cut Line= 3
      3772799.61     10571210.18      3772299.61     10572010.19
       3771149.6     10573110.19
#Sta/Elev= 30
  4118.4  312.74    4257  304.49    4415  291.34  4509.3  290.67  4670.9  286.03
    4823  286.33  4837.8  284.39  4967.5   287.6  4975.1  281.48    4981  286.26
  4990.5  282.22  4996.4  285.54  4999.8  281.43  5002.6  280.93  5005.8  281.43
  5026.4  282.67  5032.9  286.62  5374.1  286.64  5668.5   284.8  5931.9  283.88
  6091.5  293.39  6166.3   293.3  6186.3  292.74    6236  297.83  6299.5  300.61
  6459.3  319.38  6518.7  326.56  6532.9  330.36  6603.7  341.29  6653.2  343.31
#Mann= 8 ,-1 , 0
  4118.4     .12       0  4999.8     .07       0  5005.8     .12       0
  5374.1     .16       0  5668.5     .12       0  6091.5     .05       0
  6166.3     .16       0  6459.3     .12       0
Bank Sta=4967.5,5032.9
XS Rating Curve= 0 ,0
Exp/Cntr=0.3,0.1

Type RM Length L Ch R = 1 ,76473   ,751,751,751
BEGIN DESCRIPTION:
BOX CREEK 101.0
END DESCRIPTION:
XS GIS Cut Line= 3
      3772799.63     10570510.16      3771849.61     10571960.19
      3771049.61     10572760.19
#Sta/Elev= 30
  3272.6  337.36  3380.2  336.61  3461.1  332.66  3611.8  319.94  3720.3  317.34
  3762.8  310.58  3880.1   296.2  3951.6  292.07  4088.1  286.43  4196.6  284.41
  4603.2  284.77  4833.3  285.68  4992.6  286.01  5000.1  281.96  5002.9  281.46
  5006.1  281.96  5034.4  286.86  5317.3  283.98  5359.7   285.6  5402.1  283.55
  5416.2  285.11  5501.1  284.06  5600.1  286.11  5740.9  293.28  5840.5  299.33
  5991.6   314.4  6024.4  319.17  6045.6   320.2  6096.4  323.88  6137.5  327.75
#Mann= 10 ,-1 , 0
  3272.6     .16       0  3951.6     .12       0  4603.2     .16       0
  4833.3     .12       0  5000.1     .07       0  5006.1     .12       0
  5740.9     .05       0  5991.6     .16       0  6045.6     .05       0
  6096.4     .16       0
Bank Sta=4992.6,5034.4
XS Rating Curve= 0 ,0
Exp/Cntr=0.3,0.1

Type RM Length L Ch R = 1 ,75722   ,1783,1783,1783
BEGIN DESCRIPTION:
BOX CREEK 100.0
END DESCRIPTION:
XS GIS Cut Line= 3
      3772799.63     10570310.17      3771399.61     10571910.19
      3770849.58     10572410.22
#Sta/Elev= 30
  2890.3  348.01  2918.3  350.11  2954.4  347.35    2961   348.9  3173.6  324.14
  3294.2  316.38  3393.8  313.23  3506.8  303.37  3535.3  303.48  3611.5  297.31
  3667.6  292.59  3727.2  288.82  3825.7   282.9  3946.2  282.38  4428.4  282.08
  4980.8   285.1  4988.4  285.23  5006.2  279.53    5009  279.03  5012.2  279.53
    5013  282.95  5019.7  282.95  5023.5   285.6  5186.3  283.95  5283.2  286.71
  5462.3  292.39  5547.1  299.96  5674.9  315.84    5732  319.57  5759.7  322.43
#Mann= 8 ,-1 , 0
  2890.3     .16       0  3611.5     .12       0  3667.6     .16       0
  3727.2     .12       0  5006.2     .07       0  5012.2     .12       0
  5283.2     .16       0    5732      .1       0
Bank Sta=4980.8,5023.5
XS Rating Curve= 0 ,0
Exp/Cntr=0.3,0.1

Type RM Length L Ch R = 1 ,73939   ,696,696,696
BEGIN DESCRIPTION:
BOX CREEK 99.0
END DESCRIPTION:
XS GIS Cut Line= 3
      3772243.97     10569836.53      3771153.72     10571294.82
      3770528.71     10572780.96
#Sta/Elev= 30
    3569  367.08  3617.7  364.82  3788.6  335.99    3874  324.73  4117.9  300.45
  4267.9  289.91  4472.1  281.96  4638.9  278.31  4659.8  280.84  4982.9  283.39
  4986.1  278.11  4988.8  277.61  4992.1  278.11  5032.9  283.77  5096.8  283.28
  5124.6  278.56  5139.2  283.64    5160  282.76  5168.3  278.68  5196.7  283.32
  5629.8  284.09  6007.9   285.6  6048.7  285.88  6153.4  287.42    6243  291.43
  6362.9  304.62  6502.1   323.9  6697.4  325.43  6775.1  328.85    7002  331.15
#Mann= 10 ,-1 , 0
    3569     .16       0  4472.1     .12       0  4986.1     .07       0
  4992.1     .12       0  5629.8     .05       0  6007.9     .16       0
  6048.7     .12       0  6153.4     .16       0  6362.9     .05       0
  6775.1     .16       0
Bank Sta=4982.9,5032.9
XS Rating Curve= 0 ,0
Exp/Cntr=0.3,0.1

Type RM Length L Ch R = 1 ,73243   ,604,604,604
BEGIN DESCRIPTION:
BOX CREEK 98.0
END DESCRIPTION:
XS GIS Cut Line= 4
      3771973.18      10569746.2      3771021.78     10570544.82
      3770625.94     10571253.16      3769883.76     10571669.34
#Sta/Elev= 30
  3531.3  338.65  3621.9  329.79  3774.3   319.1  4026.5  302.23  4111.1  298.81
  4196.9  301.25  4260.7  295.97  4303.6  285.46  4310.1  286.52  4332.2  281.68
  4423.8  281.92  4456.7  277.24  4459.4  276.74  4462.7  277.24    4474  280.16
  4494.8  277.45    4552  281.07  4679.5  281.11  4708.1  279.29  4855.2  281.27
  4985.8   282.3  4997.9  277.61    5014   277.6    5030  282.88  5068.3  282.22
  5256.2  282.47  5696.2  284.02  5883.7  303.16  6176.5  317.19  6435.8  315.79
#Mann= 9 ,-1 , 0
  3531.3     .16       0  3774.3     .12       0  4456.7     .07       0
  4462.7     .12       0  4855.2     .16       0  4997.9     .12       0
  5068.3     .16       0  5256.2     .12       0  5883.7     .16       0
Bank Sta=4985.8,5030
XS Rating Curve= 0 ,0
Exp/Cntr=0.3,0.1

Type RM Length L Ch R = 1 ,72639   ,446,446,446
BEGIN DESCRIPTION:
BOX CREEK 97.0
END DESCRIPTION:
XS GIS Cut Line= 3
      3772049.62     10569510.18      3770499.61     10570660.19
      3770099.59     10571460.22
#Sta/Elev= 30
  3053.4  378.41  3096.2  377.63  3181.7   364.7    3211  350.56  3272.9  338.16
  3375.8  325.67  3550.4  313.69    3706  311.98    3839  312.92  3968.3  294.99
  4024.7  280.41    4311  280.67  4372.2  276.29  4374.9  275.79  4378.2  276.29
  4389.8  280.77  4796.7  281.83  4825.9  278.18  4879.9  281.72  4969.9  281.53
  4976.2  278.26  5002.3   277.2 5016.48  281.48  5019.8  277.73  5042.1  281.68
  5117.6  281.01  5489.4   281.6  5623.5  289.05  5733.2  300.93  5877.9  315.07
#Mann= 11 ,-1 , 0
  3053.4     .16       0  3272.9     .12       0  3550.4     .16       0
    3706     .12       0  4372.2     .07       0  4378.2     .12       0
  4879.9     .16       0  4976.2     .12       0  5002.3     .16       0
  5117.6     .12       0  5733.2     .16       0
Bank Sta=4969.9,5016.48
XS Rating Curve= 0 ,0
Exp/Cntr=0.3,0.1

Type RM Length L Ch R = 1 ,72193   ,733,733,733
BEGIN DESCRIPTION:
BOX CREEK 96.0
END DESCRIPTION:
XS GIS Cut Line= 3
      3771299.58     10569260.22      3770049.61     10570560.19
      3770099.61      10571360.2
#Sta/Elev= 30
  3287.9  321.13  3330.2  318.53  3351.5   314.8  3372.6  315.18  3464.7  308.13
  3556.6  306.02  3664.1  296.04  3712.2  287.63  3754.7  284.23  4299.3  278.59
  4310.5  274.98  4313.2  274.48  4316.5  274.98  4327.6  278.91  4355.9  279.61
  4688.3  280.94  4695.3  277.12  4716.6  281.02  4907.5  278.49  4978.3  281.01
  4992.4  276.83  5006.6  276.64  5013.5  281.15  5121.4  279.69  5181.5  281.13
  5281.7  279.56  5662.4   280.4  5722.6  285.64  5820.7  298.56  5892.9     307
#Mann= 5 ,-1 , 0
  3287.9     .16       0  3664.1     .12       0  4310.5     .07       0
  4316.5     .12       0  5820.7     .16       0
Bank Sta=4978.3,5013.5
XS Rating Curve= 0 ,0
Exp/Cntr=0.3,0.1

Type RM Length L Ch R = 1 ,71460   ,895,895,895
BEGIN DESCRIPTION:
BOX CREEK 95.0
END DESCRIPTION:
XS GIS Cut Line= 3
      3771149.57     10569310.22      3769899.61     10570310.19
      3769099.64     10570810.17
#Sta/Elev= 30
  3332.6  317.02    3383  318.04    3439  315.12  3542.4  297.25  3639.1  285.67
  3738.3  286.66  4108.1  279.41    4321  279.05  4335.4  277.56  4340.4   274.2
  4343.2   273.7  4346.4   274.2  4357.1  274.89  4370.7  278.95  4434.7  277.65
  4634.8  280.09  4655.6   277.3  4684.4  280.57  4818.9  278.17  4962.2  280.19
  4977.6  276.81  4998.8  277.76  5004.7  275.86  5014.1  280.17  5543.6  278.85
  5738.2  288.82    5796  295.41  5826.6   303.5  5845.3  305.81  5876.7  310.12
#Mann= 5 ,-1 , 0
  3332.6     .16       0  3542.4     .12       0  4340.4     .07       0
  4346.4     .12       0  5845.3     .16       0
Bank Sta=4962.2,5014.1
XS Rating Curve= 0 ,0
Exp/Cntr=0.3,0.1
