HEC-RAS study GASTON BRANCH.prj: GASTON BRANCH Base Level Engineering

--- GASTON BRANCH.g01 (geometry) --- (continued)

Type RM Length L Ch R = 1 ,40886   ,139,139,139
BEGIN DESCRIPTION:
GASTON BRANCH 55.0
END DESCRIPTION:
XS GIS Cut Line= 3
      3670390.99     10603449.03      3670797.25     10602830.95
      3670918.77       10602206.
#Sta/Elev= 30
  4184.4  289.21  4192.8288.5487  4208.7 287.866  4241.2  286.64  4323.1279.3109
    4428  270.37  4693.1268.9634  4955.4  270.24  4975.8  268.67    4997  260.68
  4999.8  260.18    5003  260.68  5018.3  261.52  5026.7  269.45  5108.2  268.63
  5196.7272.5398  5295.8277.2628  5328.3  282.42  5333.4  280.65  5373.1  284.87
  5403.6  285.16  5431.6  287.48  5436.7  284.51  5483.3   292.7  5488.4  290.71
  5508.1294.5537  5525.9  298.89  5534.9  299.28    5540  297.29  5560.7  298.29
#Mann= 10 ,-1 , 0
  4184.4     .05       0  4192.8     .08       0  4208.7     .05       0
  4323.1     .12       0  4693.1     .05       0    4997     .04       0
    5003     .05       0  5196.7     .16       0  5295.8     .12       0
  5508.1     .16       0
Bank Sta=4955.4,5026.7
XS Rating Curve= 0 ,0
Exp/Cntr=0.3,0.1

Type RM Length L Ch R = 1 ,40747   ,89,89,89
BEGIN DESCRIPTION:
GASTON BRANCH 54.0
END DESCRIPTION:
XS GIS Cut Line= 3
      3670481.28     10603560.12      3670887.53     10602928.18
      3671179.21     10602205.91
#Sta/Elev= 30
    4144  298.04  4201.5  293.62  4215.2  287.67  4292.9283.6555  4331.6   283.8
  4355.7 279.749  4406.7274.3824  4550.4268.2904  4634.2268.1028    4828267.9589
  4957.8  269.49  4979.4  260.24    4997  259.64  4999.8  259.14    5003  259.64
  5011.7  260.72  5024.4  269.97  5072.8269.2489  5176.9270.2918  5204.2  270.67
  5216.6  273.17  5227.4  271.02  5254.3271.6029  5335.3  274.94  5489.4291.1504
  5546.6296.2776  5593.5300.2346  5633.5  302.48  5638.9  306.99  5674.2  307.84
#Mann= 15 ,-1 , 0
    4144     .05       0  4292.9     .08       0  4355.7      .1       0
  4406.7     .05       0  4550.4     .16       0  4634.2     .05       0
    4828     .12       0    4997     .07       0    5003     .12       0
  5072.8     .16       0  5176.9     .05       0  5254.3     .16       0
  5489.4     .05       0  5546.6     .12       0  5593.5     .16       0
Bank Sta=4957.8,5024.4
XS Rating Curve= 0 ,0
Exp/Cntr=0.3,0.1

Type RM Length L Ch R = 1 ,40658   ,502,502,502
BEGIN DESCRIPTION:
Mapping XS 0572cb1f
END DESCRIPTION:
XS GIS Cut Line= 3
      3670519.46     10603660.83      3670960.44     10602983.73
      3671248.22     10602214.01
#Sta/Elev= 30
  4085.7  287.84  4223.6  288.99  4350.7286.7364    4406279.1442  4483.1  270.62
    4579266.9174  4598.8267.2231  4824.2  266.17  4959.5  268.91  4972.3   267.1
  4989.8  259.21    4997  259.13  4999.8  258.63    5003  259.13  5025.6  267.17
    5045  269.54  5135.9  267.78  5228.4269.3962  5345.9  271.45  5392.5   274.4
  5461.4282.1709  5508.3  288.99  5533.3  295.73  5563.6  297.69  5588.5  302.34
  5593.9  301.02  5641.2 305.924  5649.1  304.52  5672.1308.2765  5715.5  312.08
#Mann= 11 ,-1 , 0
  4085.7     .05       0  4350.7      .1       0    4406     .12       0
    4579     .16       0  4598.8     .12       0    4997     .07       0
    5003     .12       0  5228.4     .16       0  5461.4     .12       0
  5641.2     .16       0  5672.1     .12       0
Bank Sta=4959.5,5045
XS Rating Curve= 0 ,0
Exp/Cntr=0.3,0.1

Type RM Length L Ch R = 1 ,40156   ,264,264,264
BEGIN DESCRIPTION:
Mapping XS ee8e3bb1
END DESCRIPTION:
XS GIS Cut Line= 3
      3670845.82     10603587.93      3671311.14     10603199.01
      3671863.22     10603011.51
#Sta/Elev= 30
  4294.1  299.11    4302  300.94  4310.4296.0859  4351.4  298.38  4387.8  294.78
  4394.4  298.47    4423  294.41  4486.8  298.01  4507.6  295.67  4515.4  291.44
  4536.2  293.86    4544  288.38  4564.8  285.69  4572.6  278.93  4593.5  271.82
  4657.2  264.52  4962.3  268.22  4971.1  267.22  4976.4  259.25    4997   258.4
  4999.8   257.9    5003   258.4  5039.2  267.79  5120.7  265.84  5152.4  267.96
  5196.1  275.01  5268.6  303.51  5316.4  307.79  5390.6308.1366  5483.6  308.16
#Mann= 5 ,-1 , 0
  4294.1     .05       0  4310.4     .12       0    4997     .07       0
    5003     .12       0  5390.6     .16       0
Bank Sta=4962.3,5039.2
XS Rating Curve= 0 ,0
Exp/Cntr=0.3,0.1

Type RM Length L Ch R = 1 ,39892   ,293,293,293
BEGIN DESCRIPTION:
GASTON BRANCH 53.0
END DESCRIPTION:
XS GIS Cut Line= 2
      3670668.74     10603907.36      3671862.82     10603174.95
#Sta/Elev= 30
  4001.5   302.7  4049.6  300.64  4059.2  297.11  4080.5  296.06  4101.8  298.29
  4153.9  293.76  4159.8  296.12  4217.8  293.81  4260.6  286.46  4275.8  286.74
    4328  275.91  4401.4  270.22  4697.4  263.76  4975.7   267.7  4981.6  267.06
    4997  258.15  4999.8  257.65    5003  258.15  5024.2   260.4  5046.6  266.95
    5055  262.79  5070.1  263.63  5163.9  273.72  5192.4  280.62  5199.1  285.61
  5213.6  288.06  5244.5  299.51  5265.8  303.35  5386.8307.5722  5402.3  307.65
#Mann= 4 ,-1 , 0
  4001.5     .12       0    4997     .07       0    5003     .12       0
  5386.8     .16       0
Bank Sta=4975.7,5046.6
XS Rating Curve= 0 ,0
Exp/Cntr=0.3,0.1

Type RM Length L Ch R = 1 ,39599   ,410,410,410
BEGIN DESCRIPTION:
GASTON BRANCH 52.0
END DESCRIPTION:
XS GIS Cut Line= 3
      3671749.61      10604210.2      3671599.61     10603610.19
       3671749.6     10603460.19
#Sta/Elev= 30
    4425  295.43    4443  290.77  4469.4287.6316  4530.7  284.56  4538.4  281.37
  4571.5276.7285  4579.6  272.88    4608  268.23  4613.1  269.79  4641.5  266.15
  4703.3  262.35  4772.9  262.02    4943  265.94  4979.1  258.48    4997  257.85
  4999.8  257.35    5003  257.85  5012.6  257.99  5020.3  261.19  5025.4  258.64
  5033.2  261.78    5047  262.65  5057.6   265.5    5100  273.05  5114.2  278.71
  5128.3  280.39  5142.5  285.49  5156.6  286.39  5170.8  290.06  5255.6  290.72
#Mann= 5 ,-1 , 0
    4425     .05       0  4469.4      .1       0  4571.5     .12       0
    4997     .07       0    5003     .12       0
Bank Sta=4943,5057.6
XS Rating Curve= 0 ,0
Exp/Cntr=0.3,0.1

Type RM Length L Ch R = 1 ,39189   ,365,365,365
BEGIN DESCRIPTION:
GASTON BRANCH 51.0
END DESCRIPTION:
XS GIS Cut Line= 3
      3672049.61     10604060.22      3671999.61     10603660.19
      3671849.59     10603360.15
#Sta/Elev= 30
  4598.3  288.68  4622.8282.3896  4636.1  277.99  4668.9  272.66  4769.7  261.01
  4789.8  262.08  4920.8  263.27  4951.1  264.45  4981.3  263.34  4991.4   256.7
    4997  255.55  4999.8  255.05    5003  255.55  5023.8  256.28  5032.2   261.8
  5037.8  261.25  5046.2  263.73  5127.2  263.97    5158  262.16  5202.7  265.87
  5225.1  270.72  5233.4  274.56  5247.4  278.78  5255.8  285.46  5261.4  287.19
  5269.8  292.15  5278.2   293.4  5292.1  299.08  5314.5  302.91  5336.9  304.91
#Mann= 4 ,-1 , 0
  4598.3     .05       0  4622.8     .12       0    4997     .07       0
    5003     .12       0
Bank Sta=4981.3,5046.2
XS Rating Curve= 0 ,0
Exp/Cntr=0.3,0.1

Type RM Length L Ch R = 1 ,38824   ,387,387,387
BEGIN DESCRIPTION:
GASTON BRANCH 50.0
END DESCRIPTION:
XS GIS Cut Line= 3
      3672182.67     10604275.39      3672279.89     10603803.18
      3672044.19     10603161.94
#Sta/Elev= 30
    4589  287.42  4649.3  286.87    4676  289.17    4727  287.79    4750  289.36
  4793.8286.1595  4839.3  282.28  4931.2   269.5  4961.9  267.42  4972.1  263.06
  4982.3  256.46    4997  256.29  4999.8  255.79    5003  256.29  5023.1  261.98
  5041.7   263.4  5149.3  263.37  5204.9  261.68  5230.1  263.34  5285.7  262.12
  5340.7  263.57  5500.5  261.08  5543.1  264.81  5564.4  270.01  5611.5287.6777
  5617.7  292.78  5628.3  294.82  5640.7  301.74  5649.6  303.27  5754.3  307.71
#Mann= 5 ,-1 , 0
    4589     .05       0  4793.8     .12       0    4997     .07       0
    5003     .12       0  5611.5     .16       0
Bank Sta=4961.9,5041.7
XS Rating Curve= 0 ,0
Exp/Cntr=0.3,0.1

Type RM Length L Ch R = 1 ,38437   ,532,532,532
BEGIN DESCRIPTION:
GASTON BRANCH 49.0
END DESCRIPTION:
XS GIS Cut Line= 3
      3672040.32     10604841.35      3672644.47     10603858.73
      3672356.54     10602543.98
#Sta/Elev= 30
  3721.7  298.73  3781.5  300.11  4019.3  283.52  4077.3  288.02  4086.9  292.79
  4092.7  290.16  4108.2  297.63    4114  294.84  4166.1  301.38  4187.4  292.15
  4224.1  292.52  4266.7  300.44  4290.8296.0398  4340.1  292.31  4413.5  276.29
  4486.1  271.22  4498.6  263.38  4535.3  269.65  4976.1  261.22    4997   255.6
  4999.8   255.1    5003   255.6  5027.2  261.77  5692.7  259.43  5804.8  262.59
    5885270.2038  5995.5  284.62  6050.9  299.19  6135.2311.0113  6221.1  315.75
#Mann= 6 ,-1 , 0
  3721.7     .05       0  4290.8     .12       0    4997     .07       0
    5003     .12       0    5885     .16       0  6135.2     .05       0
Bank Sta=4976.1,5027.2
XS Rating Curve= 0 ,0
Exp/Cntr=0.3,0.1

Type RM Length L Ch R = 1 ,37905   ,576,576,576
BEGIN DESCRIPTION:
GASTON BRANCH 48.0
END DESCRIPTION:
XS GIS Cut Line= 3
      3673404.89     10604924.72      3673127.11     10603931.65
      3673182.64     10602494.71
#Sta/Elev= 30
  3787.9  301.64  3844.5  299.06  3866.8  300.58  3895.8  298.79  4047.9  297.94
  4228.7  299.21  4280.6  298.94  4309.4296.6592  4332.6   295.5  4412.3286.2325
  4567.4  271.36  4581.8   267.5  4633.7  261.55  4685.6  258.67  4960.7  258.68
    4997  253.59  4999.8  253.09    5003  253.59  5009.5  253.92  5020.7  258.91
  5230.9  256.59  5790.1256.7098  5891.4  263.34  6011.4  275.29  6071.5  284.04
  6141.5  290.58  6161.6  293.77  6171.6  297.53  6191.6  301.72  6257.1  311.32
#Mann= 6 ,-1 , 0
  3787.9     .05       0  4309.4     .16       0  4412.3     .12       0
    4997     .07       0    5003     .12       0  5790.1     .16       0
Bank Sta=4960.7,5020.7
XS Rating Curve= 0 ,0
Exp/Cntr=0.3,0.1

Type RM Length L Ch R = 1 ,37329   ,460,460,460
BEGIN DESCRIPTION:
GASTON BRANCH 47.0
END DESCRIPTION:
XS GIS Cut Line= 3
      3673599.61     10604210.16      3673649.61     10603910.19
      3673649.61      10602810.2
#Sta/Elev= 30
  4676.7  291.12  4679.2  291.12  4686.8   286.9  4696.9  285.15  4704.6  281.74
  4727.4   275.1  4770.4  268.22  4818.6  264.53  4859.2   259.6  4951.5256.7528
  4990.8  256.47    4997  249.18  4999.8  248.68    5003  249.18  5010.8  249.18
  5020.8  252.38  5030.8   257.9  5060.8  256.53  5080.8  257.93  5170.8  254.48
  5200.8   255.6  5370.8  254.29  5860.8  258.43  5900.8  263.01  5920.8  267.72
  5940.8  274.96  5950.8  280.68  6020.8  303.53  6060.8  306.84  6080.8  307.05
#Mann= 4 ,-1 , 0
  4676.7     .16       0  4951.5     .12       0    4997     .07       0
    5003     .12       0
Bank Sta=4990.8,5030.8
XS Rating Curve= 0 ,0
Exp/Cntr=0.3,0.1

Type RM Length L Ch R = 1 ,36869   ,458,458,458
BEGIN DESCRIPTION:
GASTON BRANCH 46.0
END DESCRIPTION:
XS GIS Cut Line= 3
      3674049.61     10604210.16      3674099.61     10603960.19
       3674599.6     10602760.21
#Sta/Elev= 30
    4753   275.9    4805268.1927  4904.2258.6083  4946.7  255.81  4977.3  256.53
  4987.5  250.38    4997  248.98  4999.8  248.48    5003  248.98  5010.6  250.52
  5017.1     255  5022.5  253.71  5040.4  256.47  5495.4  252.13  5701.8   254.7
  5820.4  268.59  5939.6  289.37  5985.6  294.25  6033.3  296.43  6038.7  298.46
  6062.5  300.19  6086.4  298.25  6091.8  301.48  6110.2  300.23  6139.5     304
  6187.1  305.97  6192.5  307.72  6247.6309.7454  6257.9309.7161  6307.9  309.48
#Mann= 7 ,-1 , 0
    4753     .16       0    4805     .05       0  4904.2     .12       0
    4997     .07       0    5003     .12       0  6247.6     .16       0
  6257.9     .12       0
Bank Sta=4977.3,5040.4
XS Rating Curve= 0 ,0
Exp/Cntr=0.3,0.1

Type RM Length L Ch R = 1 ,36411   ,437,437,437
BEGIN DESCRIPTION:
GASTON BRANCH 45.0
END DESCRIPTION:
XS GIS Cut Line= 3
      3674449.61     10604360.15      3674499.61     10603860.19
      3674549.61     10603260.22
#Sta/Elev= 30
  4515.9  293.08    4546  288.03  4562.8281.3226  4576.2   274.9  4586.2  272.54
  4606.3   265.3  4664.1  259.09  4716.9  261.07  4757.1  259.67  4769.6  257.57
  4807.3   255.5  4870.1   254.2    4937254.9013  4978.2  255.47  4988.2  254.18
    4997  247.84  4999.8  247.34    5003  247.84  5020.9  248.17  5028.4  254.08
  5038.4  254.93  5349.5  251.43  5359.5  252.84  5369.6   251.2  5379.6  252.61
  5442.3  250.91  5459.9  251.85  5520.1  259.44  5614.8275.1325  5620.4  276.17
#Mann= 6 ,-1 , 0
  4515.9     .16       0  4562.8     .05       0    4937     .12       0
    4997     .07       0    5003     .12       0  5614.8     .16       0
Bank Sta=4978.2,5038.4
XS Rating Curve= 0 ,0
Exp/Cntr=0.3,0.1

Type RM Length L Ch R = 1 ,35974   ,468,468,468
BEGIN DESCRIPTION:
GASTON BRANCH 44.0
END DESCRIPTION:
XS GIS Cut Line= 3
      3674995.17     10604641.86      3674864.96     10604074.15
      3675047.25     10602746.06
#Sta/Elev= 30
  4305.1  297.26  4342.3296.7636  4378.6  288.95  4409.4  286.22  4429.9  295.16
  4462.6290.8721  4563.3  274.09  4660.1  263.87  4667.3263.1665  4737.7  258.29
  4831.7254.8393  4860.8  253.05    4942  253.02    4997  246.98  4999.8  246.48
    5003  246.98  5004.9247.6831  5022.8  253.34  5335.7  250.61  5549.8  250.77
  5673.8254.3835  5745.8 260.094  5771.1  261.87  5820.2   270.3  5850.5  278.94
  5890.8  284.58  5987.4  291.17  6064.6  288.98  6131.6  296.49  6228.1  298.05
#Mann= 11 ,-1 , 0
  4305.1     .12       0  4342.3     .05       0  4462.6     .16       0
  4660.1     .12       0  4667.3     .16       0  4831.7     .05       0
    4997     .03       0    5003     .05       0  5004.9     .12       0
  5673.8     .16       0  5745.8     .12       0
Bank Sta=4942,5022.8
XS Rating Curve= 0 ,0
Exp/Cntr=0.3,0.1

Type RM Length L Ch R = 1 ,35506   ,410,410,410
BEGIN DESCRIPTION:
GASTON BRANCH 43.0
END DESCRIPTION:
XS GIS Cut Line= 3
       3675149.6      10604160.2      3675299.61     10604010.19
      3675899.63     10603410.17
#Sta/Elev= 30
  4785.5  282.36    4789  282.36  4799.7  279.16  4856.2  270.02  4870.4  265.85
  4884.5  263.79  4898.6  259.89  4912.8  258.21  4926.9  253.73  4955.2  251.07
  4983.5  252.48  4994.1  244.24    4997  244.24  4999.8  243.74    5003  244.24
  5011.8  244.37  5025.9  247.96  5054.2  251.52  5068.4  250.72  5082.5  251.79
  5124.9  251.42  5139.1   249.4  5153.2  250.36  5209.8   249.8  5351.2  252.86
  5415.9253.2782  5492.6  254.87  5605.8  262.66  5747.2  278.16  5846.2  291.84
#Mann= 4 ,-1 , 0
  4785.5     .12       0    4997     .07       0    5003     .12       0
  5415.9     .05       0
Bank Sta=4983.5,5054.2
XS Rating Curve= 0 ,0
Exp/Cntr=0.3,0.1

Type RM Length L Ch R = 1 ,35096   ,446,446,446
BEGIN DESCRIPTION:
GASTON BRANCH 42.0
END DESCRIPTION:
XS GIS Cut Line= 3
      3675449.63     10604410.17      3675599.61     10604260.19
      3676149.59      10603710.2
#Sta/Elev= 30
  4755.5  283.96  4826.2  278.15  4840.3  274.97  4854.5  270.18  4925.2  259.68
  4953.5  253.92  4964.1  248.38  4981.7  248.22    4997  244.03  4999.8  243.53
    5003  244.03    5010  244.57  5038.3  251.06    5109  248.92  5137.3  250.19
  5165.6  248.47  5179.7  250.09  5292.9  248.62  5321.2  246.78    5406  248.54
  5476.7  255.06  5490.9  257.58    5505  261.73  5519.1  263.43  5547.4  270.08
  5575.7  278.57  5589.9  281.41  5618.1  285.88  5694.9294.6742  5745.4  298.41
#Mann= 4 ,-1 , 0
  4755.5     .12       0    4997     .07       0    5003     .12       0
  5694.9     .05       0
Bank Sta=4953.5,5038.3
XS Rating Curve= 0 ,0
Exp/Cntr=0.3,0.1

Type RM Length L Ch R = 1 ,34650   ,374,374,374
BEGIN DESCRIPTION:
GASTON BRANCH 41.0
END DESCRIPTION:
XS GIS Cut Line= 3
      3675749.64     10604610.17      3675999.61     10604410.19
       3676249.6     10603810.21
#Sta/Elev= 30
  4632.4  284.61  4658.9279.3286    4710  268.16    4774  258.11  4828.7252.2867
  4874.9  248.48  4967.1  249.46    4985  245.65    4991  242.34  4996.4  244.26
    4997  242.16  4999.8  241.66  5020.2  242.16  5038.6  249.41  5044.1  249.36
  5091.7  247.59  5266.7  246.63    5310  248.37  5357.1  245.24  5410.2  253.09
  5418.4  256.56  5434.1  259.67    5440  263.91  5450.9  265.89  5457.9  270.24
  5494.2  282.92    5511  286.43  5540.2   288.7  5558.1292.6623  5602.5  297.23
#Mann= 6 ,-1 , 0
  4632.4     .16       0  4658.9     .12       0  4828.7     .16       0
  4967.1     .07       0  5044.1     .12       0  5558.1     .05       0
Bank Sta=4967.1,5038.6
XS Rating Curve= 0 ,0
Exp/Cntr=0.3,0.1

Type RM Length L Ch R = 1 ,34276   ,488,488,488
BEGIN DESCRIPTION:
GASTON BRANCH 40.0
END DESCRIPTION:
XS GIS Cut Line= 3
      3676649.61     10605510.18      3676349.61     10604410.19
      3676649.58     10604060.22
#Sta/Elev= 30
  3868.4  287.62  4193.2  268.26    4302  254.41    4416  245.84  4490.3   246.7
  4500.7   243.8  4521.4  246.32  4956.7  248.52  4977.5  248.17  4986.1  246.31
  4991.3  240.91  4999.8  239.89  5015.7  242.54  5036.6  240.39  5044.2  248.18
  5050.8  242.59  5058.5  248.09  5065.1  245.16  5079.4  248.27  5185.8  243.67
  5228.6  245.39  5320.8  258.91  5355.9  269.96  5384.5  274.33  5391.1  278.48
    5413  280.53  5419.6  284.24  5441.6  284.69  5448.1  287.38  5469.5  286.16
#Mann= 3 ,-1 , 0
  3868.4     .12       0  4956.7     .07       0  5058.5     .12       0
Bank Sta=4977.5,5044.2
XS Rating Curve= 0 ,0
Exp/Cntr=0.3,0.1

Type RM Length L Ch R = 1 ,33788   ,449,449,449
BEGIN DESCRIPTION:
GASTON BRANCH 39.0
END DESCRIPTION:
XS GIS Cut Line= 3
      3676749.61     10605360.16      3676749.61     10604460.19
      3676749.61     10604260.16
#Sta/Elev= 30
  4136.8  282.87  4176.8  279.32  4206.8  273.48  4296.8  263.03  4366.8  257.11
  4386.8  253.93  4486.8  244.73  4616.8  245.61  4626.8  242.86  4646.8  245.81
  4766.8  244.26  4956.8  247.25  4976.8  239.67    4997  239.03  4999.8  238.53
    5003  239.03  5026.8  244.33  5039.3  244.25  5046.8  247.44  5076.8  251.98
  5086.8   255.2  5116.8  260.74  5146.8  265.01  5166.8  269.78  5176.8  273.75
  5206.8  281.96  5216.8  286.95  5226.8  289.62  5234.3  293.71  5236.8  293.71
#Mann= 3 ,-1 , 0
  4136.8     .12       0    4997     .07       0    5003     .12       0
Bank Sta=4956.8,5046.8
XS Rating Curve= 0 ,0
Exp/Cntr=0.3,0.1

Type RM Length L Ch R = 1 ,33339   ,608,608,608
BEGIN DESCRIPTION:
GASTON BRANCH 38.0
END DESCRIPTION:
XS GIS Cut Line= 3
      3677149.61     10605510.18      3677149.61     10604710.19
       3676999.6     10604110.15
#Sta/Elev= 30
  4179.2   288.4  4209.2  277.14  4285.1266.1476  4339.2  256.93  4389.2  262.84
  4429.2  252.98  4449.2  254.39  4729.1244.7455  4829.2  244.84  4839.2  239.46
  4859.2  240.39  4869.2  243.62  4889.2  240.03  4899.2  243.74  4919.2  245.79
  4981.8  245.76  4989.5  238.37    4997  237.98  4999.8  237.48    5003  237.98
  5010.1  242.41  5030.7  246.45  5084.2244.8794  5278.1  245.51  5392.2255.9489
    5443  262.02  5484.3  270.26  5546.1  291.17  5571.4294.2546  5597.7  296.21
#Mann= 8 ,-1 , 0
  4179.2     .12       0  4285.1     .16       0  4729.1     .12       0
    4997     .07       0    5003     .12       0  5084.2     .16       0
  5392.2     .12       0  5571.4     .05       0
Bank Sta=4981.8,5030.7
XS Rating Curve= 0 ,0
Exp/Cntr=0.3,0.1

Type RM Length L Ch R = 1 ,32731   ,533,533,533
BEGIN DESCRIPTION:
GASTON BRANCH 37.0
END DESCRIPTION:
XS GIS Cut Line= 3
      3677701.47     10605651.25      3677636.37      10604796.2
      3677488.79     10603889.05
#Sta/Elev= 30
  4276.7   287.9  4307.9  288.96  4359.7294.5529  4436.5299.0773  4496.1  299.24
  4618.8  295.39  4627.2  294.27  4632.2  290.81  4658.9  287.81  4678.9  283.01
  4749.1   275.9  4779.2  269.91  4829.4  264.02  4894.3  253.03  4929.6  244.93
  4944.8244.0789  4969.8   241.6  4989.8   235.7    4997   235.7  4999.8   235.2
    5003   235.7  5019.9   240.8  5025.3  244.04  5170.7  243.34  5416.3 246.589
  5555.7   248.9  5827.2  273.28  5971.1  287.74  6031.9  296.27  6053.3  296.98
#Mann= 7 ,-1 , 0
  4276.7     .12       0  4359.7     .16       0  4436.5     .12       0
  4944.8     .05       0    4997     .03       0    5003     .05       0
  5416.3     .16       0
Bank Sta=4929.6,5025.3
XS Rating Curve= 0 ,0
Exp/Cntr=0.3,0.1

Type RM Length L Ch R = 1 ,32198   ,571,571,571
BEGIN DESCRIPTION:
GASTON BRANCH 36.0
END DESCRIPTION:
XS GIS Cut Line= 3
       3677899.6      10605210.2      3678149.61     10604860.19
      3678299.62     10604410.17
#Sta/Elev= 30
  4548.6  288.93  4551.7  288.93    4556  286.57  4576.9   283.3  4612.5  273.09
  4627.3   271.1  4634.6  267.78  4662.9  260.63  4734.2   247.9  4772.9243.6678
  4855.8  241.75  4923.5 242.149  4981.4  243.06  4989.3  239.98    4997  234.62
  4999.8  234.12    5003  234.62  5010.4  238.83  5020.9  242.78  5134.8240.2714
  5210.6  240.61  5305.5  252.45    5316  255.77  5347.7  261.37  5368.7  267.08
  5389.8  277.47  5400.4  279.91  5410.9  284.16    5432  288.15  5453.1  289.49
#Mann= 6 ,-1 , 0
  4548.6     .12       0  4772.9     .05       0  4923.5     .07       0
    4997     .07       0    5003     .07       0  5134.8     .12       0
Bank Sta=4981.4,5020.9
XS Rating Curve= 0 ,0
Exp/Cntr=0.3,0.1

Type RM Length L Ch R = 1 ,31627   ,573,573,573
BEGIN DESCRIPTION:
GASTON BRANCH 35.0
END DESCRIPTION:
XS GIS Cut Line= 3
      3678299.63     10605660.15      3678699.61     10604860.19
      3678649.61     10604460.18
#Sta/Elev= 30
  4124.4  296.57  4177.8289.1964  4191.7286.9524  4199.8  284.59  4205.4   281.4
  4244.5  272.19  4250.1  268.77  4303.2  257.28  4347.5251.0458  4384.3  246.51
    4429   244.4  4468.1  244.73  4607.9  240.78  4697.3  244.01  4758.8  240.59
  4804.8241.3587  4974.1  240.85  4982.4  238.35    4988  234.86    4997  232.99
  4999.8  232.49    5003  232.99  5010.4  236.32    5016  240.95  5038.9  241.41
  5069.2  244.41  5079.2  246.73  5149.8  255.85  5290.9  270.62  5421.9  275.53
#Mann= 7 ,-1 , 0
  4124.4     .07       0  4177.8     .12       0  4191.7     .07       0
  4347.5     .05       0  4804.8     .12       0    4997     .07       0
    5003     .12       0
Bank Sta=4974.1,5016
XS Rating Curve= 0 ,0
Exp/Cntr=0.3,0.1

Type RM Length L Ch R = 1 ,31054   ,481,481,481
BEGIN DESCRIPTION:
GASTON BRANCH 34.0
END DESCRIPTION:
XS GIS Cut Line= 3
      3679549.64     10605110.22      3679199.61     10604760.19
      3679049.61     10604110.18
#Sta/Elev= 30
  4519.5  275.45  4576.1  267.87  4590.2  264.87  4618.5  255.53  4655.2249.2025
  4703.4  242.93  4792.2239.5565  4844.8  237.92  4873.1  235.27  4887.2  239.18
  4986.2  239.99    4997  232.28  4999.8  231.78    5003  232.28  5017.1  232.37
  5033.3  239.96  5098.2239.8067  5271.1  238.91  5332.7  242.13  5373.7  246.13
  5404.5  251.57  5433.6  253.58  5466.1  259.13  5476.3  259.36  5486.6  262.22
  5517.4   264.8  5524.2  267.83  5529.4     267    5579  275.94  5681.6  284.44
#Mann= 6 ,-1 , 0
  4519.5     .12       0  4655.2     .05       0  4792.2     .12       0
    4997     .07       0    5003     .12       0  5098.2     .05       0
Bank Sta=4986.2,5033.3
XS Rating Curve= 0 ,0
Exp/Cntr=0.3,0.1

Type RM Length L Ch R = 1 ,30573   ,506,506,506
BEGIN DESCRIPTION:
GASTON BRANCH 33.0
END DESCRIPTION:
XS GIS Cut Line= 3
      3679599.61     10605060.17      3679599.61     10604510.19
       3679699.6     10603860.22
#Sta/Elev= 30
  4477.7  272.66  4517.7  267.17  4547.7  260.55  4580.2255.4025  4627.7  247.19
  4667.7  241.92  4707.7  238.25  4851.3238.3524  4987.7   237.5    4997  231.16
  4999.8  230.66    5003  231.16  5017.7  231.59  5025.2  238.42  5118.2237.7389
  5209.6237.3139  5300.9  237.17  5381.8  239.48  5456.4  250.14    5483  255.38
  5503.2  261.05  5513.3  262.59  5519.7  265.12  5533.6  266.93  5563.9   274.5
    5574  275.51  5587.9  280.65  5604.4  283.91  5651.2  289.19  5685.3  291.62
#Mann= 7 ,-1 , 0
  4477.7     .12       0  4580.2     .05       0  4851.3     .12       0
    4997     .07       0    5003     .12       0  5118.2     .05       0
  5209.6     .12       0
Bank Sta=4987.7,5025.2
XS Rating Curve= 0 ,0
Exp/Cntr=0.3,0.1

Type RM Length L Ch R = 1 ,30067   ,522,522,522
BEGIN DESCRIPTION:
GASTON BRANCH 32.0
END DESCRIPTION:
XS GIS Cut Line= 3
      3680099.61      10604910.2      3680099.61     10604510.19
      3680149.61     10604010.19
#Sta/Elev= 30
  4612.8   264.8  4625.3264.5875  4682.8  262.48  4722.8   259.1  4762.8   250.5
  4772.8  247.35  4802.8  242.25  4862.8  235.96  4882.8  235.06  4982.8  235.88
    4997  230.92  4999.8  230.42    5003  230.92  5010.3   232.8  5015.3   232.8
  5022.9  236.43    5043  237.02  5173.6  235.24    5254  237.27  5294.2  240.82
  5314.3  243.73  5354.5  253.84  5365.2255.2145  5374.6  257.35  5424.9  264.13
  5462.5  273.22  5467.6  272.85  5475.1  274.92  5495.2  276.27  5515.3  275.89
#Mann= 5 ,-1 , 0
  4612.8     .05       0  4625.3     .12       0    4997     .07       0
    5003     .12       0  5365.2     .16       0
Bank Sta=4982.8,5022.9
XS Rating Curve= 0 ,0
Exp/Cntr=0.3,0.1

Type RM Length L Ch R = 1 ,29545   ,565,565,565
BEGIN DESCRIPTION:
GASTON BRANCH 31.0
END DESCRIPTION:
XS GIS Cut Line= 3
       3680399.6     10604910.22      3680499.61     10604210.19
      3680249.58     10603860.15
#Sta/Elev= 30
  4286.2  262.53  4328.5259.5283    4367  256.28  4417.6  249.69  4498.4  244.31
  4518.6  241.45  4579.2  240.58  4649.9  236.71  4750.9  234.86  4902.4  236.23
  4973.1  235.72  4996.4  233.38    4997  230.69  4999.8  230.19    5003  230.69
  5021.6  230.81  5030.2  235.37  5051.1  238.94    5072  239.78    5154251.9313
  5165.4  254.01  5172.8  256.89  5193.6  259.51  5229.3   268.4  5251.4  271.75
  5258.8   271.8  5264.9  273.97  5323.9  281.34  5414.7287.9045  5423.5  288.37
#Mann= 6 ,-1 , 0
  4286.2     .05       0  4328.5     .12       0    4997     .07       0
    5003     .12       0    5154     .16       0  5414.7     .05       0
Bank Sta=4973.1,5051.1
XS Rating Curve= 0 ,0
Exp/Cntr=0.3,0.1

Type RM Length L Ch R = 1 ,28980   ,538,538,538
BEGIN DESCRIPTION:
GASTON BRANCH 30.0
END DESCRIPTION:
XS GIS Cut Line= 3
      3680199.59     10605510.23      3681049.61     10604110.19
      3680849.61     10603710.18
#Sta/Elev= 30
  3373.6  298.29  3412.3296.6533  3482.2  293.03  3767.1   268.5  3788.4  269.15
  3904.7   265.4  4131.5  255.08  4538.5  239.79  4636.4238.7159  4777.5  234.27
  4881.6  234.27  4939.7  231.98  4961.1  234.05  4966.9  232.37  4976.4  235.21
  4982.4  230.89  4988.3  231.05    4997  228.47  4999.8  227.97    5003  228.47
  5014.3  229.61  5019.9  234.94  5042.2  232.66  5064.6  235.21    5154  233.62
  5226.7  237.26  5271.4  244.02  5346.9  260.99    5414  273.22  5458.7  274.66
#Mann= 5 ,-1 , 0
  3373.6     .12       0  3412.3     .05       0  4636.4     .12       0
    4997     .07       0    5003     .12       0
Bank Sta=4976.4,5019.9
XS Rating Curve= 0 ,0
Exp/Cntr=0.3,0.1

Type RM Length L Ch R = 1 ,28442   ,543,543,543
BEGIN DESCRIPTION:
GASTON BRANCH 29.0
END DESCRIPTION:
XS GIS Cut Line= 3
      3681299.61     10605060.18      3681549.61     10603960.19
       3681349.6     10603510.17
#Sta/Elev= 30
  3874.4  262.73  3905.2  260.34  3941.6  255.25  3989.8  254.54  4110.3  247.59
  4223.1  243.42  4484.1  237.13  4653.8  234.54    4939234.0841  4961.4  233.58
  4971.7  232.97  4978.3  228.79  4983.5   231.6    4997  227.81  4999.8  227.31
    5003  227.81  5016.8  231.75  5034.6  234.59  5115.3  234.09  5138.5  232.85
  5248.8233.9162  5306.8  236.08  5341.7  242.23  5358.8  247.13  5405.3  263.98
  5418.3   271.7  5428.5  273.83  5440.2  280.38  5457.3  283.51  5494.9  286.48
#Mann= 5 ,-1 , 0
  3874.4     .05       0    4939     .16       0    4997     .07       0
    5003     .16       0  5248.8     .12       0
Bank Sta=4961.4,5034.6
XS Rating Curve= 0 ,0
Exp/Cntr=0.3,0.1

Type RM Length L Ch R = 1 ,27899   ,570,570,570
BEGIN DESCRIPTION:
GASTON BRANCH 28.0
END DESCRIPTION:
XS GIS Cut Line= 3
      3683299.63     10605210.21      3682049.61     10603810.19
      3681399.59     10603410.18
#Sta/Elev= 30
  3135.5  287.02  3744.6  246.54    3773  248.53  3829.8  247.33    4028  237.11
  4169.3  233.44  4495.3  231.36  4623.2  232.95  4680.4236.3188  4764.5  246.22
  4792.9  243.94    4828  237.51    4864  231.11  4976.8  232.15    4997  225.22
  4999.8  224.72    5003  225.22  5015.3  226.69  5025.9  232.23  5035.5  232.67
  5106.3  231.36    5165  234.18  5376.4  233.95    5529  238.71  5589.4249.1084
  5646.1  258.71  5673.2  265.05  5688.6  271.01  5746.6  283.14  5775.6  285.01
#Mann= 5 ,-1 , 0
  3135.5     .05       0  4680.4     .16       0    4997     .07       0
    5003     .16       0  5589.4     .12       0
Bank Sta=4828,5529
XS Rating Curve= 0 ,0
Exp/Cntr=0.3,0.1

Type RM Length L Ch R = 1 ,27329   ,538,538,538
BEGIN DESCRIPTION:
GASTON BRANCH 27.0
END DESCRIPTION:
XS GIS Cut Line= 3
       3683399.6     10604510.18      3682599.61     10603710.19
      3681799.63     10602910.21
#Sta/Elev= 30
  3887.4  269.68  3972.2   261.5  4099.5  253.25  4354.1  241.98  4410.6  241.78
  4537.9  235.19  4606.1233.0885  4754.4230.3529  4798.4230.1321  4863.2  230.21
  4905.6  229.05  4976.3  231.14  4990.5  224.79    4997  224.35  4999.8  223.85
    5003  224.35  5004.6  224.35  5015.2  232.25  5103.6  230.34    5443  234.78
  5658.3235.8987  5757.3237.0216  5810.7   236.9  5890.7239.1635  5892.8 239.162
  5923.9  239.37  5966.3  241.24  6038.2250.7232  6079.4  254.91  6150.1  266.53
#Mann= 11 ,-1 , 0
  3887.4     .05       0  4606.1     .16       0  4754.4     .12       0
  4798.4     .16       0    4997     .07       0    5003     .16       0
  5658.3     .12       0  5757.3     .16       0  5890.7     .12       0
  5892.8     .16       0  6038.2     .12       0
Bank Sta=4976.3,5015.2
XS Rating Curve= 0 ,0
Exp/Cntr=0.3,0.1

Type RM Length L Ch R = 1 ,26791   ,452,452,452
BEGIN DESCRIPTION:
GASTON BRANCH 26.0
END DESCRIPTION:
XS GIS Cut Line= 3
       3683849.6     10604260.18      3683049.61     10603460.19
      3682249.63     10602660.21
#Sta/Elev= 30
  3864.6  284.37  3963.6  276.61  4161.6  255.35  4373.7  239.07  4486.8  235.47
  4670.7  235.19  4770.6230.4119    4798   229.4  4852.6232.3945  4925.2  233.09
  4981.8  230.92  4987.3226.9092  4992.4  223.19    4997  222.52  4999.8  222.02
    5003  222.52  5010.1  222.52  5024.2  227.82  5052.5  229.92  5186.8228.9813
  5420.2  230.43  5434.4  232.55  5533.4  230.57  5762.9233.0986  5844.5  233.32
  5929.9237.7166  5957.6   240.3  5971.8  243.96  6009.1248.5389  6127.3   261.1
#Mann= 10 ,-1 , 0
  3864.6     .05       0  4770.6     .12       0  4852.6     .16       0
  4987.3     .12       0    4997     .07       0    5003     .12       0
  5186.8     .16       0  5762.9     .12       0  5929.9     .16       0
  6009.1     .05       0
Bank Sta=4981.8,5052.5
XS Rating Curve= 0 ,0
Exp/Cntr=0.3,0.1

Type RM Length L Ch R = 1 ,26339   ,662,662,662
BEGIN DESCRIPTION:
GASTON BRANCH 25.0
END DESCRIPTION:
XS GIS Cut Line= 3
      3684006.18     10604079.22      3683480.12     10603297.94
       3682658.2     10602293.95
#Sta/Elev= 30
  3943.3  271.37  3998.1  264.48  4019.1  264.74  4155.7 250.302    4322  236.63
  4450.2231.2528  4588.9  226.91  4903.3228.0179  4990.4  229.13    4997  222.68
  4999.8  222.18    5003  222.68  5011.5  222.85  5019.1  228.92  5047.8   227.1
  5171.2228.3765  5352.8  231.22  5523.7  240.77  5603.9242.8077  5686.6  243.41
    5800  248.11    5907  253.54    5950  258.35  5970.8  258.05  6034.7   268.2
    6057   274.6  6063.4  273.45  6077.8  280.81  6106.5   286.3  6182.7  287.85
#Mann= 8 ,-1 , 0
  3943.3     .16       0  4155.7     .05       0  4450.2     .16       0
  4903.3     .12       0    4997     .07       0    5003     .12       0
  5171.2     .16       0  5603.9     .05       0
Bank Sta=4990.4,5019.1
XS Rating Curve= 0 ,0
Exp/Cntr=0.3,0.1

Type RM Length L Ch R = 1 ,25677   ,289,289,289
BEGIN DESCRIPTION:
Mapping XS 583b1f43
END DESCRIPTION:
XS GIS Cut Line= 3
      3684495.75     10604178.15       3684094.7     10603287.52
      3683277.69     10602574.59
#Sta/Elev= 30
  3949.1  298.07  4091.2280.3797  4563.6  233.16  4652.9230.1701  4875.5  225.61
  4970.4   227.2  4984.7  222.73    4997  222.03  4999.8  221.53    5003  222.03
  5013.6 222.493  5040.7  227.84  5083.4  228.98  5154.6   234.6  5253.3  247.11
  5310.3  247.89  5324.5  245.84  5381.5  244.79  5421.1245.9424  5430.8  243.87
  5522.9  245.52  5579.9  242.39  5600.7  243.97  5671.9  242.62  5735.5  246.77
    5764  246.63  5862.7  254.65  5919.7  255.73  5948.2  254.04  6010.2  257.68
#Mann= 7 ,-1 , 0
  3949.1     .16       0  4091.2     .05       0  4652.9     .16       0
    4997     .07       0    5003     .16       0  5013.6     .12       0
  5421.1     .05       0
Bank Sta=4970.4,5040.7
XS Rating Curve= 0 ,0
Exp/Cntr=0.3,0.1

Type RM Length L Ch R = 1 ,25388   ,133,133,133
BEGIN DESCRIPTION:
GASTON BRANCH 24.0
END DESCRIPTION:
XS GIS Cut Line= 3
      3684912.44     10603615.68      3684474.91     10603183.36
      3683386.37     10602537.53
#Sta/Elev= 30
  4133.1  276.51  4160.2   272.8  4344.1  261.13  4447.4257.1014    4512252.3677
  4549.1  250.42  4592.6244.5934    4646 239.533  4754.4  230.07  4887.2225.4333
  4939.2225.8631    4952  226.54    4997  222.24  4999.8  221.74    5003  222.24
  5017.5  227.59    5113  226.84  5184.6  229.95  5235.7  236.47  5251.3  244.05
    5275248.2852  5350.5 254.831  5449.4  262.66    5491     265  5570.9  264.97
  5761.9  257.48  5841.8  259.63  5921.7   265.5  5967.5264.7643  6013.9  264.77
#Mann= 13 ,-1 , 0
  4133.1     .05       0  4447.4     .08       0    4512     .05       0
  4592.6     .08       0    4646     .05       0  4887.2     .16       0
  4939.2     .05       0    4997     .04       0    5003     .05       0
    5275     .12       0  5350.5     .08       0  5449.4     .05       0
  5967.5     .08       0
Bank Sta=4952,5017.5
XS Rating Curve= 0 ,0
Exp/Cntr=0.3,0.1

Type RM Length L Ch R = 1 ,25255   ,249,249,249
BEGIN DESCRIPTION:
GASTON BRANCH 23.0
END DESCRIPTION:
XS GIS Cut Line= 2
      3685032.19     10603360.43      3683460.51     10602444.49
#Sta/Elev= 30
  4151.1  272.19  4219.4  270.39  4321.2  261.52  4358.4  262.31  4385.7  258.96
  4395.6   261.5  4422.9  258.42  4438.6  260.32  4460.1  252.03  4475.8   252.3
  4524.6  242.71  4679.3  228.75  4759.5  226.27  4929.6  227.05  4972.9  224.42
  4978.7  226.26    4997  222.31  4999.8  221.81    5003  222.31  5015.9  222.31
  5031.7  226.68  5037.4  224.09  5154.9  228.42  5293.9  242.88    5381   258.6
    5513  264.85  5550.3  271.24  5747.9   267.5  5828.2  270.41  5970.2  280.75
#Mann= 3 ,-1 , 0
  4151.1     .05       0    4997     .03       0    5003     .05       0
Bank Sta=4978.7,5031.7
XS Rating Curve= 0 ,0
Exp/Cntr=0.3,0.1

Type RM Length L Ch R = 1 ,25006   ,241,241,241
BEGIN DESCRIPTION:
Mapping XS e4c91d0f
END DESCRIPTION:
XS GIS Cut Line= 3
      3685125.94     10603292.72      3684490.54     10602777.11
      3683516.57     10602365.65
#Sta/Elev= 30
  4034.1  269.02  4125.7  267.88  4239.2  259.98    4538  229.16  4686.7  225.27
  4884.3226.1922  4958.3  226.18  4972.8  222.99    4982  224.23    4997  222.26
  4999.8  221.76    5003  222.26  5037.4225.5432  5048.8  226.78  5140.5  225.49
  5269.9  232.28  5293.6  236.05  5346.4  238.44  5370.1  241.65  5399.3  241.65
  5499.5  248.62  5528.7  248.49  5546.9  251.01  5552.4  249.54  5576.1  253.61
  5628.9  255.08  5652.6  258.54  5758.3  265.56    5782  270.05  5909.7  284.19
#Mann= 5 ,-1 , 0
  4034.1     .05       0  4884.3     .12       0    4997     .07       0
    5003     .12       0  5037.4     .05       0
Bank Sta=4958.3,5048.8
XS Rating Curve= 0 ,0
Exp/Cntr=0.3,0.1

Type RM Length L Ch R = 1 ,24765   ,797,797,797
BEGIN DESCRIPTION:
GASTON BRANCH 22.0
END DESCRIPTION:
XS GIS Cut Line= 3
      3685214.48     10603235.42      3684698.87     10602610.44
      3683438.44     10602198.98
#Sta/Elev= 30
  3999.6  261.97    4014  260.37  4034.8  262.12  4077.8  260.47  4176.8  260.94
  4262.8  257.33    4298   258.9  4333.2  256.17  4411.3  241.09  4433.5  239.81
  4489.5  231.64  4752.7  224.59  4953.3  225.78    4997  222.17  4999.8  221.67
    5003  222.17  5022.4  225.94  5442.2   224.3  5482.3  225.59  5500.7  228.02
    5506  225.87  5564.5  230.46  5665.5  234.82  5761.1  245.61  5776.8  245.89
    5793  248.86  5862.1  255.74  6039.8  283.82    6080  286.46  6135.7  283.27
#Mann= 3 ,-1 , 0
  3999.6     .05       0    4997     .03       0    5003     .05       0
Bank Sta=4953.3,5022.4
XS Rating Curve= 0 ,0
Exp/Cntr=0.3,0.1

Type RM Length L Ch R = 1 ,23968   ,615,615,615
BEGIN DESCRIPTION:
GASTON BRANCH 21.0
END DESCRIPTION:
XS GIS Cut Line= 3
      3685399.62     10602710.21      3684949.61     10602010.19
      3683349.64      10601610.2
#Sta/Elev= 30
  4196.1  260.76  4406.5  247.37  4666.7  237.52  4760.5  236.85  4890.6  227.56
  4965.6 222.492  4984.4  223.89  4992.6  223.23    4997  220.01  4999.8  219.51
    5003  220.01  5014.7  223.96  5157.1224.3543  5257.6   222.2  5265.4  220.01
  5368.4  222.32  5440.6  220.01  5646.8  220.01  5664.8  222.24  5669.9  220.01
  5729.2  220.01  5739.5  222.18  5894.1  222.53  6131.2  227.89  6296.1  232.27
  6388.9  240.77  6448.2  253.28  6512.6  251.69  6613.1  262.55  6677.5  263.89
#Mann= 5 ,-1 , 0
  4196.1     .05       0  4965.6     .12       0    4997     .07       0
    5003     .12       0  5157.1     .05       0
Bank Sta=4890.6,6131.2
XS Rating Curve= 0 ,0
Exp/Cntr=0.3,0.1

Type RM Length L Ch R = 1 ,23353   ,322,322,322
BEGIN DESCRIPTION:
GASTON BRANCH 20.0
END DESCRIPTION:
XS GIS Cut Line= 3
      3685399.61     10602510.22      3685449.61     10601910.19
      3684649.62      10601310.2
#Sta/Elev= 30
  4391.5  251.93  4511.9  242.15  4622.3  230.96  4702.6  228.86  4762.8   230.5
  4810.5  226.59  4815.5   227.2  4923.4  221.87  4996.7  221.27    4997  220.01
  4999.8  219.51    5003  220.01  5012.7221.7782  5165.5  222.52  5257.2  220.62
  5286.3  223.11  5350.9  222.59  5371.7   221.2  5545.3222.1914  5649.7222.2077
  5681.5  222.22  5700.9  221.87  5707.2  220.01  5786.3  220.14  5843.6  227.52
  5915.5  237.36  5943.6  242.19  5950.9  244.87  5980.1  246.84  5993.6  245.86
#Mann= 7 ,-1 , 0
  4391.5     .05       0    4997     .03       0    5003     .05       0
  5012.7     .12       0  5545.3     .05       0  5649.7     .12       0
  5681.5     .05       0
Bank Sta=4815.5,5843.6
XS Rating Curve= 0 ,0
Exp/Cntr=0.3,0.1

Type RM Length L Ch R = 1 ,23031   ,378,378,378
BEGIN DESCRIPTION:
GASTON BRANCH 19.0
END DESCRIPTION:
XS GIS Cut Line= 3
      3685716.23      10603144.7      3685750.95     10601912.09
      3684761.91     10598823.49
#Sta/Elev= 30
  3575.7  268.64  3730.3  259.33  3810.3  250.99  3869.3  249.94  4110.4  228.58
  4240.5  220.65  4337.7  220.01  4462.1  220.01  4560.6  220.01  4730.7     229
  4971.9220.7014    4997  220.01  4999.8  219.51    5003  220.01  5169.8  220.01
    5283  220.01  5652.7  220.01  5797.8  256.13  5877.7  263.23    6108  256.12
  6186.3   260.8    6274  260.26  6600.7  247.62  6793.5  253.12  6964.8  247.26
  7125.5  246.73  7250.9253.6547  7572.4   266.9  7912.7   272.4  8051.9  277.97
#Mann= 9 ,-1 , 0
  3575.7     .05       0  4337.7     .07       0  4462.1     .05       0
  4971.9     .12       0    4997     .07       0    5003     .12       0
  5169.8      .1       0    5283     .05       0  7250.9     .16       0
Bank Sta=4110.4,4730.7
XS Rating Curve= 0 ,0
Exp/Cntr=0.3,0.1

Type RM Length L Ch R = 1 ,22653   ,898,898,898
BEGIN DESCRIPTION:
GASTON BRANCH 18.0
END DESCRIPTION:
XS GIS Cut Line= 3
      3685829.95     10603235.26       3685986.2     10601998.32
      3686884.63      10598990.5
#Sta/Elev= 30
  3559.6  274.83    3839  252.62  4068.7  227.23  4119.1  221.86  4149.3  222.57
  4159.9  220.01  4229.4  220.01  4683.1  220.01  4814.9  223.01    4997  220.01
  4999.8  219.51    5003  220.01  5047.2  220.01  5257.4  220.01  5359.4  220.01
    5423  220.01  5539.8  220.01  5855.5221.1177  5940.9220.8658  6641.2223.1068
  6703.9  227.47  6776.9   234.3  6792.5  233.97  6930.2  249.38  7057.6257.9937
  7111.5  261.17  7361.4  264.02  7716.2  258.45  7838.4  257.73  7945.5  259.81
#Mann= 14 ,-1 , 0
  3559.6     .05       0  4229.4     .07       0  4683.1     .05       0
    4997     .03       0    5003     .05       0  5047.2     .12       0
  5257.4     .07       0  5359.4     .05       0    5423     .07       0
  5539.8     .05       0  5855.5     .12       0  5940.9     .05       0
  6641.2     .12       0  7057.6     .05       0
Bank Sta=4068.7,6703.9
XS Rating Curve= 0 ,0
Exp/Cntr=0.3,0.1

Type RM Length L Ch R = 1 ,21755   ,521,521,521
BEGIN DESCRIPTION:
GASTON BRANCH 17.0
END DESCRIPTION:
XS GIS Cut Line= 4
      3686749.61     10602910.17      3686699.61     10602310.19
      3686699.61     10601995.73      3687129.64      10599780.5
#Sta/Elev= 30
  4420.6  262.33  4437.8260.1389  4483.3  253.07  4523.3246.1454  4642.2224.6628
  4671.4  220.34  4740.9  220.01  4850.8  220.01  4942.9  220.01    4997  220.01
  4999.8  219.51    5003  220.01  5152.7  222.64  5233.2232.9435  5292.7  245.65
  5342.8   251.5  5417.5  249.31  5572.6  229.84  5658.6  224.02  5836.2  235.31
  5933.6  234.09  6203.2  249.45  6290.1  245.92  6432.7  257.81  6518.6  256.28
  6713.3241.0274    6848244.4147  6950.1249.5611  7237.5  259.36  7593.7  256.02
#Mann= 13 ,-1 , 0
  4420.6     .16       0  4437.8     .12       0  4523.3     .16       0
  4642.2     .05       0  4740.9     .07       0  4850.8     .05       0
  4942.9     .07       0    4997     .07       0    5003     .07       0
  5233.2     .05       0  6713.3     .12       0    6848     .05       0
  6950.1     .12       0
Bank Sta=4483.3,5342.8
XS Rating Curve= 0 ,0
Exp/Cntr=0.3,0.1

Type RM Length L Ch R = 1 ,21234   ,530,530,530
BEGIN DESCRIPTION:
GASTON BRANCH 16.0
END DESCRIPTION:
XS GIS Cut Line= 3
      3686849.63     10602910.14      3687199.61     10602160.19
      3686749.59     10601910.18
#Sta/Elev= 30
  4185.6  260.79  4262.8  252.01  4273.8  248.33  4306.9  244.44  4313.6242.7697
  4319.6  241.21  4351.1  238.32  4365.3  235.62  4405.6232.0652  4419.9229.5624
  4450.4   227.1  4462.2  225.25  4502.4  222.56  4526.2221.9955  4593.9  220.01
  4738.8  220.01    4997  220.01  4999.8  219.51    5003  220.01    5277  220.01
  5314.1  220.01  5344.9  223.26  5367.8  227.54    5425  236.14  5447.9  240.98
  5454.8  243.43  5492.5   247.3  5514.3  248.31    5520  246.61    5528  247.09
#Mann= 9 ,-1 , 0
  4185.6     .12       0  4313.6     .16       0  4405.6     .05       0
  4419.9     .16       0  4526.2     .05       0  4738.8     .07       0
    4997     .07       0    5003     .07       0    5277     .05       0
Bank Sta=4450.4,5367.8
XS Rating Curve= 0 ,0
Exp/Cntr=0.3,0.1

Type RM Length L Ch R = 1 ,20704   ,515,515,515
BEGIN DESCRIPTION:
GASTON BRANCH 15.0
END DESCRIPTION:
XS GIS Cut Line= 3
      3689049.63      10602860.2      3687649.61     10601910.19
      3687249.63     10601310.21
#Sta/Elev= 30
  3316.3  298.97  3401.7  299.85  3410.6  291.09  3425.1  285.74  3431.6  276.14
  3461.3  259.49  3503.5  255.64  3533.4  262.67  3560.4  252.58  3569.3  243.56
  3654.4237.1512  3707.6236.9324    3791  234.35  3824.1227.2127  3839.7220.3093
  4004.8  220.01  4369.8  220.01  4620.4  225.04  4669.9  220.01  4808.6  220.01
    4997  220.01  4999.8  219.51    5003  220.01  5217.9  220.01  5397.3  220.07
  5412.3  227.42  5418.7227.4158  5448.4  235.18  5536.2242.4674  5729.3  255.64
#Mann= 14 ,-1 , 0
  3316.3     .05       0  3654.4     .08       0  3707.6     .05       0
  3824.1     .16       0  3839.7     .05       0  4004.8     .07       0
  4369.8     .12       0  4669.9     .05       0  4808.6     .07       0
    4997     .07       0    5003     .07       0  5217.9     .05       0
  5418.7     .16       0  5536.2     .05       0
Bank Sta=4620.4,5412.3
XS Rating Curve= 0 ,0
Exp/Cntr=0.3,0.1

Type RM Length L Ch R = 1 ,20189   ,581,581,581
BEGIN DESCRIPTION:
GASTON BRANCH 14.0
END DESCRIPTION:
XS GIS Cut Line= 3
      3688849.63     10602360.21      3688149.61     10601760.19
       3687349.6     10601260.18
#Sta/Elev= 30
  4066.4  246.67  4070.5246.4485  4102.1  231.92    4123  231.11  4137.2  226.13
    4180  226.14  4194.3  225.81  4210.4222.7719  4215.2  221.47  4250.8  220.01
    4997  220.01  4999.8  219.51    5003  220.01  5067.5220.9624  5111.6  222.33
  5196.8220.9209  5376.1220.9058  5444.2222.8501  5495.5   226.2    5568  231.42
  5619.9  232.23  5625.8  234.59  5635.2  233.67  5641.1  235.41  5675.2237.3073
  5720.1  238.21  5735.4  240.21  5866.3  246.29  5924.1   250.5  5931.8  252.13
#Mann= 10 ,-1 , 0
  4066.4     .05       0  4070.5     .16       0  4210.4     .05       0
    4997    .035       0    5003     .05       0  5067.5     .12       0
  5196.8     .05       0  5376.1     .12       0  5444.2     .16       0
  5675.2     .05       0
Bank Sta=4180,5495.5
XS Rating Curve= 0 ,0
Exp/Cntr=0.3,0.1

Type RM Length L Ch R = 1 ,19608   ,566,566,566
BEGIN DESCRIPTION:
GASTON BRANCH 13.0
END DESCRIPTION:
XS GIS Cut Line= 3
       3689099.6     10602810.17      3688599.61     10601410.19
      3687299.64      10601010.2
#Sta/Elev= 30
  3529.4  312.14  3539.5  313.64  3570.3  294.43  3601.1  288.31  3614.3  271.63
  3637.2  262.55  3693.4  257.87    3763  246.63  3794.8  246.45  3858.6  253.11
  3872.9  248.21  3881.5248.5347  3903.7  249.55  3922.3  246.35    3983247.5572
  4070.9   248.3  4083.1   244.9  4092.2  237.41  4108.6  229.61    4117225.2564
  4171.5221.5783    4997  220.01  4999.8  219.51    5003  220.01  5347.5  220.01
  5633.3  226.49  5741.4228.4008  5877.7234.0656  6009.9  238.37  6376.1  256.99
#Mann= 10 ,-1 , 0
  3529.4     .05       0  3881.5      .1       0    3983     .05       0
    4117     .16       0  4171.5     .05       0    4997    .033       0
    5003     .05       0  5347.5     .12       0  5741.4     .16       0
  5877.7     .05       0
Bank Sta=4108.6,5633.3
XS Rating Curve= 0 ,0
Exp/Cntr=0.3,0.1

Type RM Length L Ch R = 1 ,19042   ,550,550,550
BEGIN DESCRIPTION:
GASTON BRANCH 12.0
END DESCRIPTION:
XS GIS Cut Line= 3
      3689549.62     10602610.22      3689049.61     10601060.19
      3688649.62     10599760.21
#Sta/Elev= 30
  3407.7   315.2  3423.8  314.03  3439.3  308.27  3449.8  293.28  3455.8  290.88
  3512.8   286.1    3616  288.03  3621.3  286.42  3628.4   277.6  3638.9  271.42
  3648.1  261.01  3680.1  247.88    3744   243.9    3807  233.56  4048.7  225.76
  4164.3  226.02  4171.4  230.57  4227.3  228.96  4279.8  220.82  4321.9  220.01
    4997  220.01  4999.8  219.51    5003  220.01  5402.4220.9141  5538.6  226.63
  5595.7228.6581    5738  232.73  5901.5  243.04  6314.8  259.01  6396.5  259.68
#Mann= 5 ,-1 , 0
  3407.7     .05       0    4997    .033       0    5003     .05       0
  5402.4     .12       0  5595.7     .05       0
Bank Sta=4227.3,5538.6
XS Rating Curve= 0 ,0
Exp/Cntr=0.3,0.1

Type RM Length L Ch R = 1 ,18492   ,328,328,328
BEGIN DESCRIPTION:
GASTON BRANCH 11.0
END DESCRIPTION:
XS GIS Cut Line= 3
       3689750.6     10602541.05      3689449.61     10600710.19
      3688899.61     10600060.19
#Sta/Elev= 30
  3131.8  287.64  3284.7  286.46    3305  289.46  3315.1  286.27  3335.4  271.85
  3352.1  253.14  3357.2  255.31  3361.3  251.79  3365.8  247.92    3386  243.55
  3418.4  240.87  3461.3  232.18  3700.2  227.09  3730.6  231.88    3761  231.62
  3771.1  237.54  3791.4  239.43  3841.9  238.85  3852.2  234.75  3872.5  224.82
  3913.3  220.92    4997  220.01  4999.8  219.51    5003  220.01  5134.9  220.01
  5280.3  229.48  5306.4  232.22  5398.7  238.85  5661.3  241.62  5838.7   247.9
#Mann= 7 ,-1 , 0
  3131.8     .05       0  3361.3      .1       0  3461.3     .05       0
    4997    .033       0    5003     .05       0  5134.9     .12       0
  5280.3     .05       0
Bank Sta=3852.2,5306.4
XS Rating Curve= 0 ,0
Exp/Cntr=0.3,0.1

Type RM Length L Ch R = 1 ,18164   ,504,504,504
BEGIN DESCRIPTION:
GASTON BRANCH 10.0
END DESCRIPTION:
XS GIS Cut Line= 3
3689946.5517578910602510.2179532      3689649.61     10600460.19
      3689149.61      10599710.2
#Sta/Elev= 30
  2629.9  238.41  2897.9  238.41  2907.2  242.97  2912.3   247.5  2918.1   260.7
  2928.2  264.01  2938.3  261.86  2948.4  257.77  2958.6  249.25  2968.7  245.43
  2977.5  236.88  2982.5  240.59    2999  235.46  3029.3  232.89  3187.1  231.27
  3263.5  231.22  3286.8  229.99  3386.5  227.58  3423.4  227.45  3433.5  225.22
  3443.6  220.96  3453.7  220.01  5219.6  220.01  5225.5  220.01  5293.8  220.01
  5316.4  221.49  5427.9  224.27  5496.6  226.82  5667.9  240.98  5870.7  251.05
#Mann= 7 ,-1 , 0
  2629.9     .05       0  3187.1      .1       0  3286.8     .15       0
  3386.5     .05       0  5219.6     .07       0  5225.5     .12       0
  5427.9     .05       0
Bank Sta=3423.4,5316.4
XS Rating Curve= 0 ,0
Exp/Cntr=0.3,0.1

Type RM Length L Ch R = 1 ,17660   ,255,255,255
BEGIN DESCRIPTION:
Mapping XS 1a6ad100
END DESCRIPTION:
XS GIS Cut Line= 3
3690021.9285697810602420.2040976      3689955.46     10601682.38
      3689972.82     10599174.45
#Sta/Elev= 30
  2445.1  234.48  2671.7  234.48  2701.8  232.31    2732  231.78  2937.6  229.83
    3003  228.31  3103.5  228.94  3161.3  227.96    3199  226.94    3204   227.3
  3213.9  230.63    3244  228.49  3260.1  229.09  3304.3  220.83  3314.9  220.01
  4594.7  220.01  4614.7  221.29  4694.7  221.84  4804.7  220.83  4814.7  221.83
  4846.9  220.01    5105  220.77  5134.7  221.93  5265.7  227.04  5334.7  228.84
  5434.7  236.24  5494.7  241.92  5614.8  248.73  5814.8  251.85  5920.5  254.81
#Mann= 7 ,-1 , 0
  2445.1     .05       0  2937.6     .15       0  3161.3      .1       0
  3260.1     .05       0  4846.9     .07       0    5105     .12       0
  5265.7     .05       0
Bank Sta=4814.7,5134.7
XS Rating Curve= 0 ,0
Exp/Cntr=0.3,0.1
