--- GUM CREEK.prj (project) ---

Proj Title=GUM CREEK Base Level Engineering
Current Plan=p01
Default Exp/Contr=0.3,0.1
English Units
Geom File=g01
Flow File=f01
Plan File=p01
Y Axis Title=Elevation
X Axis Title(PF)=Main Channel Distance
X Axis Title(XS)=Station
BEGIN DESCRIPTION:
GUM CREEK
END DESCRIPTION:
DSS Export Rating Curves= 0
DSS Export Rating Curve Sorted= 0
DSS Export Volume Flow Curves= 0
DXF OffsetX= 0
DXF OffsetY= 0
DXF ScaleX= 1
DXF ScaleY= 10

--- GUM CREEK.p01 (plan) ---

Plan Title=Multiple Run
Short Identifier=Multiple
Geom File=g01
Flow File=f01
Subcritical Flow
K Sum by GR= 0
Std Step Tol= 0.01
Critical Tol= 0.01
Num of Std Step Trials= 20
Max Error Tol= 0.3
Flow Tol Ratio= 0.001
Split Flow NTrial= 30
Split Flow Tol= 0.02
Split Flow Ratio= 0.02
Log Output Level= 0
Friction Slope Method= 1
Unsteady Friction Slope Method= 2
Unsteady Bridges Friction Slope Method= 1
Parabolic Critical Depth
Global Vel Dist=  1 , 1 , 1
Global Log Level= 0
CheckData=True
Encroach Param= -1, 0, 0, 0
BEGIN DESCRIPTION:
Multiple Run
END DESCRIPTION:

--- GUM CREEK.f01 (steady flow) ---

Flow Title=Multiple
Program Version=4.10
Number of Profiles= 7
Profile Names=10-year,25-year,50-year,1pct_min,100-year,1pct_plu,500-year
River Rch & RM=GUM CREEK,Reach-1         ,34785
     377     500     600     531     717     970    1029
River Rch & RM=GUM CREEK,Reach-1         ,30325
     633     864    1057     952    1288    1741    1915
River Rch & RM=GUM CREEK,Reach-1         ,27299
    1172    1671    2106    1950    2638    3567    4153
River Rch & RM=GUM CREEK,Reach-1         ,27017
    1172    1671    2106    1950    2638    3567    4153
River Rch & RM=GUM CREEK,Reach-1         ,26789
    1431    2046    2583    2393    3236    4377    5101
River Rch & RM=GUM CREEK,Reach-1         ,26310
    1431    2046    2583    2393    3236    4377    5101
River Rch & RM=GUM CREEK,Reach-1         ,20200
    1503    2146    2705    2501    3382    4574    5310
River Rch & RM=GUM CREEK,Reach-1         ,14867
    1899    2729    3456    3206    4335    5863    6852
River Rch & RM=GUM CREEK,Reach-1         ,8327
    1966    2822    3570    3307    4472    6048    7051
River Rch & RM=GUM CREEK,Reach-1         ,1685
    2014    2892    3659    3390    4584    6200    7228
Boundary for River Rch & Prof#=GUM CREEK,Reach-1         , 1
Up Type= 0
Dn Type= 3
Dn Slope=0.004
Boundary for River Rch & Prof#=GUM CREEK,Reach-1         , 2
Up Type= 0
Dn Type= 3
Dn Slope=0.004
Boundary for River Rch & Prof#=GUM CREEK,Reach-1         , 3
Up Type= 0
Dn Type= 3
Dn Slope=0.004
Boundary for River Rch & Prof#=GUM CREEK,Reach-1         , 4
Up Type= 0
Dn Type= 3
Dn Slope=0.004
Boundary for River Rch & Prof#=GUM CREEK,Reach-1         , 5
Up Type= 0
Dn Type= 3
Dn Slope=0.004
Boundary for River Rch & Prof#=GUM CREEK,Reach-1         , 6
Up Type= 0
Dn Type= 3
Dn Slope=0.004
Boundary for River Rch & Prof#=GUM CREEK,Reach-1         , 7
Up Type= 0
Dn Type= 3
Dn Slope=0.004
DSS Import GetInterval= 0
DSS Import GetPeak= 0
DSS Import FillOption= 0

--- GUM CREEK.g01 (geometry) ---

Geom Title=Existing Conditions
Program Version=4.10

River Reach=GUM CREEK       ,Reach-1
Reach XY= 30
      3749500.32     10609465.14      3748790.75       10609679.
      3748093.25       10611168.       3747943.5       10612628.
      3748129.25       10613041.       3747757.5       10613973.
      3746428.75       10615777.      3745556.25       10615554.
      3745268.25       10616321.      3743959.75       10617741.
      3743239.75       10617502.      3742534.75       10617780.
      3741914.75       10617463.      3741180.75       10617497.
        3740784.       10617234.      3740567.25       10616457.
        3738485.       10615100.       3737104.5       10615486.
        3735639.       10615097.        3734712.       10615155.
      3733732.25       10616023.       3733276.5       10617299.
      3733346.75       10618184.      3732871.75       10618656.
      3733096.75       10618841.       3733061.5       10619457.
       3732675.5       10619372.      3731182.25       10620194.
       3730784.5       10620054.        3729982.       10620492.

Type RM Length L Ch R = 1 ,34785   ,323,323,323
BEGIN DESCRIPTION:
Mapping XS a6f41992
END DESCRIPTION:
XS GIS Cut Line= 2
      3749186.23      10609327.1      3749505.66     10609906.94
#Sta/Elev= 30
  4706.2  409.27  4719.5  409.31  4725.2  410.04  4732.3  408.72  4741.3  409.67
  4768.8  410.43  4844.5  411.25    4872  412.44  4909.8  411.79  4915.5  413.01
  4938.1  412.75  4991.2  412.11  4997.5  413.21    5013  412.11  5018.7  413.03
  5034.8  413.06  5050.8  412.17  5056.6  412.82  5078.3  412.65  5094.4  411.77
  5100.1  412.27  5132.2  412.12    5138  411.49  5143.7   412.2  5181.5  412.22
  5241.2  411.13  5246.9  411.61  5284.7  411.36  5314.8  410.46  5368.2  411.26
#Mann= 3 , 0 , 0
  4706.2     .16       0  4938.1     .07       0  4997.5     .16       0
Bank Sta=4938.1,4997.5
XS Rating Curve= 0 ,0
Exp/Cntr=0.3,0.1

Type RM Length L Ch R = 1 ,34462   ,46,46,46
BEGIN DESCRIPTION:
GUM CREEK 71.0
END DESCRIPTION:
XS GIS Cut Line= 3
       3749149.6     10609510.21      3749048.55     10609753.85
      3749299.59     10609910.18
#Sta/Elev= 30
  4725.8  407.17  4841.3  404.03  4855.7  405.06  4870.6  404.82  4877.3  404.08
  4894.5  404.97  4909.8  404.59  4918.4   401.2  4923.8   402.6  4931.5  400.48
  4942.3  398.05  4947.7  398.47  4953.1  397.03  4971.6  396.02  4989.6  396.02
  4991.4  395.57  4994.1  395.07  4997.4  395.57  5037.9   395.8  5061.5  397.29
  5067.6  399.82  5073.5  400.12  5082.9  402.15  5104.2   402.3    5110  401.73
    5162  403.03  5183.2  402.95  5226.4  404.51    5250  404.09  5285.3  405.37
#Mann= 3 ,-1 , 0
  4725.8     .16       0  4991.4     .07       0  4997.4     .16       0
Bank Sta=4931.5,5067.6
XS Rating Curve= 0 ,0
Exp/Cntr=0.3,0.1

Type RM Length L Ch R = 1 ,34416   ,35,35,35
BEGIN DESCRIPTION:
Mapping XS ed40f18b
END DESCRIPTION:
XS GIS Cut Line= 3
      3748851.98     10609332.49      3749018.66     10609787.37
      3749411.01     10610020.01
#Sta/Elev= 30
  4520.1  401.31  4647.4   401.1  4728.3  399.54  4773.3  400.55    4845  399.53
  4875.5  400.06  4922.4  402.67  4931.2  399.65  4936.5  399.06  4943.7  396.99
  4961.7  395.18  5012.7  395.07  5015.4  394.57  5018.7  395.07  5037.1  395.12
  5074.2  396.63  5095.6  397.86  5101.4  398.76  5110.3  402.15  5122.8   400.9
  5159.9  401.43  5168.4  402.18  5203.3  402.59  5218.4  402.13  5249.6   403.2
  5276.8  403.17  5313.9  404.79  5393.8  406.33  5400.9     407  5460.7  407.25
#Mann= 3 ,-1 , 0
  4520.1     .16       0  5012.7     .07       0  5018.7     .16       0
#XS Ineff= 2 , 0
         4861.59  401.43
Permanent Ineff=
       F       F
Bank Sta=4931.2,5101.4
XS Rating Curve= 0 ,0
Exp/Cntr=0.3,0.1

Type RM Length L Ch R = 1 ,34381   ,382,382,382
BEGIN DESCRIPTION:
Mapping XS d71cf050
END DESCRIPTION:
XS GIS Cut Line= 3
      3748782.53     10609339.41      3748970.04     10609787.37
      3749323.15     10610015.85
#Sta/Elev= 30
  4495.3  400.37  4660.1   399.9  4821.4  397.07  4853.9   398.2  4861.3  396.67
  4866.7  397.88  4885.1  397.73  4890.5  399.39  4914.3  399.36  4919.7  401.34
  4938.1  402.11  4961.9  400.56  4967.3  397.88  4983.6  398.55  4990.8   395.7
  4996.8  396.71    5009  395.15  5011.7  394.65    5015  395.15  5048.2  395.85
  5054.2  397.65  5069.3  398.78  5084.5  398.96  5090.5  400.47  5105.6  399.63
  5111.6   402.7  5126.7  403.03  5141.9  400.99  5235.6  401.48  5401.5  404.92
#Mann= 3 ,-1 , 0
  4495.3     .16       0    5009     .07       0    5015     .16       0
#XS Ineff= 2 , 0
         4915.45   401.3
Permanent Ineff=
       F       F
Bank Sta=4983.6,5069.3
XS Rating Curve= 0 ,0
Exp/Cntr=0.3,0.1

Type RM Length L Ch R = 1 ,33999   ,389,389,389
BEGIN DESCRIPTION:
Mapping XS 34639560
END DESCRIPTION:
XS GIS Cut Line= 4
      3748438.48     10609313.34      3748730.17     10609722.23
      3748889.02     10609904.52      3749352.03     10610099.89
#Sta/Elev= 30
  4422.3   406.8  4485.3  406.03  4506.1   403.7  4627.8  400.22  4636.4  401.41
  4657.3  399.66    4701  400.23  4814.7  396.49  4972.6  395.78  4986.9  394.32
  4990.5  392.15  4993.3  391.65  4996.5  392.15  5007.8  394.18    5022  393.84
  5036.2  395.79  5045.5  395.92  5120.8  396.06    5135  395.73  5142.6  393.97
  5156.8  396.21    5194  396.13  5217.7  397.75    5276  396.99  5376.3  400.28
  5476.5  401.15    5482  402.52  5568.6  404.86  5586.6  404.19  5668.9  404.92
#Mann= 5 ,-1 , 0
  4422.3     .05       0  4990.5     .03       0  4996.5     .05       0
  5045.5     .16       0  5586.6     .05       0
Bank Sta=4972.6,5036.2
XS Rating Curve= 0 ,0
Exp/Cntr=0.3,0.1

Type RM Length L Ch R = 1 ,33610   ,468,468,468
BEGIN DESCRIPTION:
GUM CREEK 70.0
END DESCRIPTION:
XS GIS Cut Line= 3
      3748049.57     10609510.15      3748663.13     10610114.97
       3749199.6     10610060.19
#Sta/Elev= 30
  4173.8  417.44  4435.5  405.63  4697.1  398.88  4711.2   394.3  4739.5  392.09
  4789.1  391.94  4824.4  398.14  4859.8  393.09  4921.6  392.83  4937.5  391.18
  4958.8   386.6  4991.1  385.92  4993.9  385.42  4997.1  385.92  5041.9  390.94
  5082.1  391.98  5102.2  386.12  5112.2  386.11  5129.4  387.71  5134.5  393.05
  5142.4  394.37  5162.5   394.2  5182.6  388.93  5192.6  388.69  5202.7  389.72
  5212.7  393.48    5263     395    5273  396.95  5484.1  399.56  5574.6  403.41
#Mann= 4 ,-1 , 0
  4173.8     .05       0  4921.6     .16       0  4991.1     .07       0
  4997.1     .16       0
Bank Sta=4937.5,5082.1
XS Rating Curve= 0 ,0
Exp/Cntr=0.3,0.1

Type RM Length L Ch R = 1 ,33142   ,74,74,74
BEGIN DESCRIPTION:
GUM CREEK 69.0
END DESCRIPTION:
XS GIS Cut Line= 2
       3748047.8     10610449.45      3748971.42     10610584.87
#Sta/Elev= 30
  4615.4  396.66  4718.3  394.01  4799.2  390.52  4820.1  391.19  4858.3  389.93
    4880  388.77  4895.8  386.63  4937.7  385.83  4940.4  385.33  4943.7  385.83
  5061.9   385.9  5102.4  387.52  5122.6  386.18  5213.5  386.31  5223.6  386.56
  5234.1  389.85    5254  387.24  5272.3  388.09  5277.3  390.62  5294.4  386.39
  5314.6  390.26  5324.7  389.44  5342.1  389.73  5347.1  391.68  5365.1  393.73
  5395.5  393.03  5405.6  394.85  5411.9  394.05  5532.4  395.93  5548.9  396.32
#Mann= 7 ,-1 , 0
  4615.4     .05       0  4820.1     .16       0  4895.8     .05       0
  4937.7    .033       0  4943.7     .05       0  5234.1     .16       0
  5532.4     .05       0
Bank Sta=4858.3,5234.1
XS Rating Curve= 0 ,0
Exp/Cntr=0.3,0.1

Type RM Length L Ch R = 1 ,33068   ,72,72,72
BEGIN DESCRIPTION:
Mapping XS 7b01985c
END DESCRIPTION:
XS GIS Cut Line= 2
      3748059.98      10610518.9      3748905.92     10610652.37
#Sta/Elev= 30
  4658.8  395.57  4739.4  393.63  4826.5  389.37  4850.8  390.08  4869.3  389.04
    4894  387.85  4931.8  390.64  4951.4  390.83  4956.4  389.31  4972.3  390.85
  5002.6  391.59  5018.9  390.15    5033  392.08  5053.2  391.73  5063.4  389.15
  5073.5  388.85  5081.3  389.32  5086.4  390.98  5093.7  391.18    5114   389.7
  5124.1  389.97  5134.2  389.13  5140.8  385.04  5143.5  384.54  5146.8  385.04
  5154.5  385.71  5164.6  390.03  5216.4  389.51  5263.4  390.63  5515.2  396.23
#Mann= 5 ,-1 , 0
  4658.8     .05       0  4869.3     .16       0  5140.8     .07       0
  5146.8     .16       0  5263.4     .05       0
Bank Sta=5124.1,5164.6
XS Rating Curve= 0 ,0
Exp/Cntr=0.3,0.1

Type RM Length L Ch R = 1 ,32996   ,298,298,298
BEGIN DESCRIPTION:
Mapping XS 218cfbd2
END DESCRIPTION:
XS GIS Cut Line= 2
      3748039.12     10610591.81      3748881.22     10610708.14
#Sta/Elev= 30
  4669.4  395.65  4780.9  391.24  4831.4  389.95  4861.7   387.5  4881.9  388.72
  4902.1  388.63  4918.6  386.87  4952.6  386.38  4962.6  385.24  4982.1  382.95
  4987.1  383.03  4992.9  380.61  5020.2  380.44    5023  379.94  5026.2  380.44
  5043.4  381.68  5064.1   384.5    5104  384.95  5114.1   384.4  5124.2   380.9
  5135.9  380.86  5144.4  384.95  5154.5  386.26  5194.8  388.12  5298.1  391.23
  5326.1  392.44  5396.7  393.01  5406.8  394.26  5428.5  393.75  5519.5  395.93
#Mann= 5 ,-1 , 0
  4669.4     .05       0  4918.6     .16       0  5020.2     .07       0
  5026.2     .16       0  5298.1     .05       0
Bank Sta=4962.6,5064.1
XS Rating Curve= 0 ,0
Exp/Cntr=0.3,0.1

Type RM Length L Ch R = 1 ,32698   ,569,569,569
BEGIN DESCRIPTION:
GUM CREEK 68.0
END DESCRIPTION:
XS GIS Cut Line= 3
      3748049.57     10610710.16      3748249.61     10610860.19
      3748549.65     10611010.21
#Sta/Elev= 30
  4727.5  392.97  4784.8   390.4  4824.4  388.08    4864  386.56  4905.7  386.34
  4920.3  384.67  4934.8  383.87    4964  384.04  4974.4  382.26  4980.3  382.26
  4985.9  379.71  5005.3  379.07    5008  378.57  5011.3  379.07  5013.9  379.68
  5044.6  381.69    5067  382.09  5097.7  383.62  5120.1  383.58  5125.7   384.5
  5134.1  383.35  5142.5  382.91    5148  384.79  5156.4  386.24  5170.4  385.56
  5201.2  387.06  5215.1  386.84  5231.9  387.74  5259.8  387.92    5313  389.47
#Mann= 4 ,-1 , 0
  4727.5     .05       0  4824.4     .16       0  5005.3     .07       0
  5011.3     .16       0
Bank Sta=4980.3,5044.6
XS Rating Curve= 0 ,0
Exp/Cntr=0.3,0.1

Type RM Length L Ch R = 1 ,32129   ,398,398,398
BEGIN DESCRIPTION:
GUM CREEK 67.0
END DESCRIPTION:
XS GIS Cut Line= 3
       3747679.2     10611152.26      3748061.12     10611301.56
      3748545.88     10611343.11
#Sta/Elev= 30
  4485.4   391.9  4546.6     390  4606.3  389.38  4625.4  388.47  4630.8  389.14
  4769.2  383.91  4793.7  381.86  4818.2     382    4848  380.18  4883.2  379.42
    4904  376.68  4924.1  377.67  4954.2  376.88  4971.2  375.23    4974  374.73
  4977.2  375.23  5004.4  376.62  5024.4  379.91  5044.5  381.47  5057.3  381.66
  5074.6  383.13  5134.8  385.93  5164.9  386.25  5171.1  387.22  5215.1  388.74
  5235.2  388.55  5275.3  389.57  5295.4   390.4  5305.5  391.57    5382  391.52
#Mann= 3 ,-1 , 0
  4485.4     .16       0  4971.2     .07       0  4977.2     .16       0
Bank Sta=4954.2,5004.4
XS Rating Curve= 0 ,0
Exp/Cntr=0.3,0.1

Type RM Length L Ch R = 1 ,31731   ,435,435,435
BEGIN DESCRIPTION:
GUM CREEK 66.0
END DESCRIPTION:
XS GIS Cut Line= 3
      3747699.62      10611360.2      3747999.61     10611660.19
      3748299.56     10611660.19
#Sta/Elev= 30
  4579.8  394.02  4636.4  391.08  4678.8  387.88  4692.9  386.41  4735.3  383.54
  4763.6  382.15  4777.8  380.78  4791.9  380.45  4806.1  378.75  4834.3  376.87
  4862.6  377.12  4876.8  377.77  4919.2  377.52  4955.8  376.53  5027.9  375.39
    5044  375.37    5061  374.43  5063.8  373.93    5067  374.43    5094  374.43
    5104  375.89    5114  375.26    5124   377.7    5144  379.87    5164  381.03
    5174   382.2    5204  384.53    5214  384.91    5224  386.02    5304  390.69
#Mann= 5 ,-1 , 0
  4579.8     .16       0  4955.8     .12       0  5027.9     .16       0
    5061     .07       0    5067     .16       0
Bank Sta=5044,5104
XS Rating Curve= 0 ,0
Exp/Cntr=0.3,0.1

Type RM Length L Ch R = 1 ,31296   ,516,516,516
BEGIN DESCRIPTION:
GUM CREEK 65.0
END DESCRIPTION:
XS GIS Cut Line= 3
      3747649.62     10612110.19      3747949.61     10612110.19
      3748249.61     10611860.19
#Sta/Elev= 30
  4669.6  390.59  4689.6  389.98  4709.6  388.44  4759.6  386.12  4819.6  382.21
  4829.6  382.04  4839.6  381.16  4869.6  379.78  4879.6   378.5  4889.6  377.84
  4919.6  376.86  4927.2  376.15  4949.6  374.47  4956.6  374.43  4959.3  373.93
  4962.6  374.43  5045.6  374.43  5147.3  374.56  5161.6  376.01  5168.1  377.38
  5178.6  377.66  5196.7  380.02  5203.9  379.37  5231.9  380.69  5239.7  381.74
  5246.2  381.56    5282  382.69    5310   384.5  5346.4  385.63  5360.1  386.78
#Mann= 6 ,-1 , 0
  4669.6     .16       0  4927.2     .12       0  4956.6     .07       0
  4962.6     .12       0  5045.6     .05       0  5178.6     .16       0
Bank Sta=4919.6,5168.1
XS Rating Curve= 0 ,0
Exp/Cntr=0.3,0.1

Type RM Length L Ch R = 1 ,30780   ,258,258,258
BEGIN DESCRIPTION:
GUM CREEK 64.0
END DESCRIPTION:
XS GIS Cut Line= 3
      3747649.61     10612410.19      3747949.61     10612610.19
      3748249.62     10612560.19
#Sta/Elev= 30
  4645.4  385.38  4681.5  383.82    4695  383.82    4710   382.8    4725  383.05
    4731  382.37    4740  382.82  4767.1  382.57  4817.8  380.54  4825.7  379.52
  4839.2  379.21  4861.7  376.99  4875.2  376.34  4884.3  375.05  4894.8  374.43
  4897.5  373.93  4900.8  374.43  5160.6  374.43  5178.3  376.43  5188.4  376.69
  5198.6  377.75  5216.3  380.94  5221.4  380.26    5229  381.55  5245.9  382.67
  5269.5  384.66  5277.1  384.86  5282.2  384.14  5289.8  385.48  5310.1  386.87
#Mann= 5 ,-1 , 0
  4645.4     .16       0  4817.8     .05       0  4894.8    .033       0
  4900.8     .05       0  5245.9     .16       0
Bank Sta=4875.2,5178.3
XS Rating Curve= 0 ,0
Exp/Cntr=0.3,0.1

Type RM Length L Ch R = 1 ,30522   ,89,89,89
BEGIN DESCRIPTION:
Mapping XS fd46a809
END DESCRIPTION:
XS GIS Cut Line= 4
      3747477.32     10612954.03      3747845.37     10612964.44
      3748083.21     10612796.04       3748270.7     10612566.89
#Sta/Elev= 30
  4446.3  383.98  4485.5  382.71  4490.5  383.55  4498.6   383.6  4508.6  382.86
  4528.6   382.7  4548.6  381.25  4628.7  379.13  4668.7  376.94  4698.7  376.65
  4718.7  375.69  4728.7  376.29  4744.6  375.33  4775.7  374.43  4778.5  373.93
  4781.7  374.43  5150.6  374.43  5171.5  376.51  5178.1  377.93  5185.8  378.27
  5200.2  380.14    5221  380.01  5242.7  381.72  5249.7   381.1  5262.3  381.34
  5284.9  382.97  5299.2  384.87  5327.9  384.98  5348.8  386.27    5402  387.58
#Mann= 5 ,-1 , 0
  4446.3     .16       0  4744.6     .05       0  4775.7    .033       0
  4781.7     .05       0  5262.3     .16       0
Bank Sta=4728.7,5171.5
XS Rating Curve= 0 ,0
Exp/Cntr=0.3,0.1

Type RM Length L Ch R = 1 ,30433   ,80,80,80
BEGIN DESCRIPTION:
Mapping XS 26e82deb
END DESCRIPTION:
XS GIS Cut Line= 4
      3747473.88     10613047.78      3747892.24     10613047.78
      3748083.21     10612901.94      3748282.86     10612591.19
#Sta/Elev= 30
  4370.9  387.27  4496.6  382.96  4606.6  381.05  4626.6  377.01  4656.6   379.2
  4776.6  378.31  4799.2  376.84  4810.7  374.43  4813.5  373.93  4816.7  374.43
  4827.6  374.43  5065.2  374.43  5071.2  378.35  5079.2  374.62  5086.4  374.43
  5092.3  377.65  5101.6  375.68  5107.5  380.07  5114.8  377.86  5122.7  377.56
  5128.6  379.89  5137.9  376.49  5143.8  381.96    5159  379.34    5165  381.42
  5207.3  380.68    5268  381.35  5295.1  385.13  5361.8  387.77  5398.9  387.99
#Mann= 5 ,-1 , 0
  4370.9     .16       0  4810.7    .033       0  4816.7     .16       0
  4827.6     .05       0  5207.3     .16       0
Bank Sta=4799.2,5071.2
XS Rating Curve= 0 ,0
Exp/Cntr=0.3,0.1

Type RM Length L Ch R = 1 ,30353   ,28,28,28
BEGIN DESCRIPTION:
Mapping XS 7857f87a
END DESCRIPTION:
XS GIS Cut Line= 5
      3747411.33     10613240.49      3747921.76     10613112.01
      3748031.13     10613051.25      3748131.83     10612959.23
      3748334.76     10612575.91
#Sta/Elev= 30
  4250.2  391.71  4391.6  385.46  4537.2  376.07  4568.1  376.95  4575.4  374.43
  4578.2  373.93  4581.4  374.43  4645.7  374.43  4790.9  375.68  4806.9  374.43
  4812.7   376.3  4828.7  375.44  4834.4  377.07  4850.4  374.43  4877.9  377.39
  4888.2  375.51  4915.3  376.74  4936.9  374.43  4943.7  375.86  4951.1  374.43
  5138.8  374.43  5147.7  377.31  5169.7  379.29  5204.3  379.98    5252  380.09
  5279.7  383.85    5296  383.77  5301.7  386.16  5345.7  388.03  5471.8  389.22
#Mann= 6 ,-1 , 0
  4250.2     .05       0  4391.6     .16       0  4575.4    .033       0
  4581.4     .16       0  4645.7     .05       0  5204.3     .16       0
Bank Sta=4568.1,4790.9
XS Rating Curve= 0 ,0
Exp/Cntr=0.3,0.1

Type RM Length L Ch R = 1 ,30325   ,393,393,393
BEGIN DESCRIPTION:
GUM CREEK 63.0
END DESCRIPTION:
XS GIS Cut Line= 4
      3747409.59     10613287.36      3747907.87     10613174.51
      3748235.99     10612915.83       3748355.2     10612561.68
#Sta/Elev= 30
  4224.7  393.43  4296.5  390.94    4358  387.94  4409.3  384.93    4415  384.09
    4440  383.37  4458.2  381.33  4482.8  379.82  4501.3  379.01  4522.1  377.13
  4532.3  377.16  4546.6  374.43  4549.3  373.93  4552.6  374.43  4606.1  374.43
  5169.9  374.43  5183.1  376.42    5191  376.36  5201.6  378.48  5222.7  378.84
  5240.8  380.68  5254.3  382.96  5260.2  383.21    5286  385.57  5317.6  387.06
  5423.2  388.87  5454.8   388.6  5475.9  389.58  5507.6  388.98  5527.1  389.56
#Mann= 6 ,-1 , 0
  4224.7     .05       0  4482.8     .16       0  4546.6    .033       0
  4552.6     .16       0  4606.1     .05       0  5260.2     .16       0
Bank Sta=4532.3,5183.1
XS Rating Curve= 0 ,0
Exp/Cntr=0.3,0.1

Type RM Length L Ch R = 1 ,29932   ,420,420,420
BEGIN DESCRIPTION:
GUM CREEK 62.0
END DESCRIPTION:
XS GIS Cut Line= 3
      3747499.61     10613410.19      3747949.61     10613360.19
      3748349.64     10613360.19
#Sta/Elev= 30
    4529  394.99  4539.1   394.1  4549.1  393.86  4579.3  391.17  4589.4  390.87
  4609.5  389.33  4629.6  387.59  4639.7  385.85  4669.9  383.96    4700  380.76
  4710.1  380.05  4720.2  378.22  4730.2   377.5  4740.3  375.53  4760.4  375.69
  4767.5  374.43  4770.2  373.93  4773.5  374.43  5188.1  374.43  5211.8  374.74
  5221.8  375.82  5231.8  375.79  5241.8   376.5  5261.8  379.11  5281.8  380.29
  5291.8  380.35  5311.8  381.85  5361.8  384.09  5371.8  384.03  5381.8   384.6
#Mann= 4 ,-1 , 0
    4529     .05       0  4767.5    .033       0  4773.5     .05       0
  5188.1     .16       0
Bank Sta=4760.4,5221.8
XS Rating Curve= 0 ,0
Exp/Cntr=0.3,0.1

Type RM Length L Ch R = 1 ,29512   ,231,231,231
BEGIN DESCRIPTION:
GUM CREEK 61.0
END DESCRIPTION:
XS GIS Cut Line= 3
      3747549.57     10613510.16      3747849.61     10613760.19
      3748299.58     10613710.19
#Sta/Elev= 30
    4608  392.13  4621.7   391.4    4636  390.08  4643.8  388.56  4664.7  387.19
  4672.5  385.02    4679  385.71  4693.3  383.37  4699.8     383  4707.6  381.65
  4714.1  381.65  4728.5   380.2  4736.3  378.66  4742.8   378.8  4757.1  376.57
  4764.3  376.45  4774.9  374.43  4777.7  373.93  4780.9  374.43  5149.5  374.43
  5209.9  378.51  5219.9  378.44    5230  379.76    5240  379.62  5310.5  382.49
  5340.7  383.02  5350.7  384.17  5380.9  383.79  5392.5  384.27  5451.3  385.65
#Mann= 4 ,-1 , 0
    4608     .05       0  4774.9    .033       0  4780.9     .05       0
  5392.5     .16       0
Bank Sta=4742.8,5209.9
XS Rating Curve= 0 ,0
Exp/Cntr=0.3,0.1

Type RM Length L Ch R = 1 ,29281   ,58,58,58
BEGIN DESCRIPTION:
Mapping XS caafbff0
END DESCRIPTION:
XS GIS Cut Line= 2
      3747394.47     10613763.37      3748283.35     10614273.78
#Sta/Elev= 30
  4580.9  392.59  4598.4   391.8  4604.4  390.54    4626  389.88  4647.5  386.44
  4663.3  386.22  4679.1  385.14  4684.9  384.25  4706.5  382.87  4713.7  381.88
  4722.3   381.7    4728  380.78  4749.6  379.14  4765.4  377.87  4771.3  374.67
  4778.2  374.43    4781  373.93  4784.2  374.43  5367.5  374.43  5462.8  374.43
  5468.6  375.62  5484.4  375.12  5490.1   375.9  5505.9  375.47  5511.7  376.32
  5520.9  376.35  5534.1  377.85  5543.3  378.48  5592.2  379.44  5605.9  380.45
#Mann= 5 ,-1 , 0
  4580.9     .05       0  4778.2    .033       0  4784.2     .05       0
  5367.5     .16       0  5534.1     .05       0
Bank Sta=4749.6,5543.3
XS Rating Curve= 0 ,0
Exp/Cntr=0.3,0.1

Type RM Length L Ch R = 1 ,29223   ,75,75,75
BEGIN DESCRIPTION:
GUM CREEK 60.0
END DESCRIPTION:
XS GIS Cut Line= 3
       3747344.2     10613801.28      3747740.89     10614028.18
      3748244.02     10614335.59
#Sta/Elev= 30
  4561.2  394.92    4646  388.84  4659.6   386.5    4705   384.2  4732.3  380.25
  4785.6  379.08  4791.3  377.73  4807.2  378.88  4901.5  378.96  4952.5  377.69
  4968.4  379.17  5127.8  377.82  5164.5   378.9  5201.3  377.35  5207.2  378.42
  5219.6  375.26  5222.4  374.76  5225.6  375.26  5228.5  378.45  5238.1   375.7
  5243.9  377.79  5259.4  375.62  5265.2  377.56  5280.7  375.72  5286.5  377.98
  5296.1  376.33    5302   378.3  5369.6  376.69  5491.6  379.75  5607.8  380.19
#Mann= 4 ,-1 , 0
  4561.2     .05       0  5219.6    .033       0  5225.6     .05       0
  5369.6     .16       0
Bank Sta=5207.2,5228.5
XS Rating Curve= 0 ,0
Exp/Cntr=0.3,0.1

Type RM Length L Ch R = 1 ,29148   ,338,338,338
BEGIN DESCRIPTION:
Mapping XS 8c23f340
END DESCRIPTION:
XS GIS Cut Line= 3
      3747118.14     10613651.73      3747306.92     10613868.73
      3748210.39     10614377.92
#Sta/Elev= 30
  4281.6  398.78  4327.3  399.45  4444.5  399.25  4487.3  397.34  4515.8   397.5
  4617.8  390.46  4652.7  386.51  4661.1  387.16  4675.6  385.89  4720.4   381.3
  4763.7  374.33  4813.4  371.69  4850.3   371.4  4863.3  369.01    4866  368.51
  4869.3  369.01  5158.1  369.01  5168.2   371.1    5174  370.24  5180.7  372.79
  5211.6  373.32  5217.3  372.43  5233.2  373.61  5254.9  373.52  5292.5  376.12
  5319.9  375.52  5364.3   377.4  5461.7  379.23  5503.4  380.52  5606.3  380.22
#Mann= 5 ,-1 , 0
  4281.6     .16       0  4327.3     .05       0  4863.3    .033       0
  4869.3     .05       0  5461.7     .16       0
Bank Sta=4850.3,5168.2
XS Rating Curve= 0 ,0
Exp/Cntr=0.3,0.1

Type RM Length L Ch R = 1 ,28810   ,240,240,240
BEGIN DESCRIPTION:
Mapping XS f9243e22
END DESCRIPTION:
XS GIS Cut Line= 2
      3746684.92     10614142.15      3748029.87     10614485.55
#Sta/Elev= 30
  4190.5   385.7  4288.5  383.83    4319  384.54  4528.5   381.6  4556.6   380.4
  4564.2  379.32  4569.3  379.85    4605  377.24  4610.2  377.89  4645.9  374.24
    4651  375.06  4659.8  374.16  4686.7  370.05  4691.9   371.1  4718.7  369.01
  4721.5  368.51  4724.7  369.01  4753.3  369.01  5192.3  369.32  5212.6  370.86
  5217.8  370.42  5227.4  371.43  5248.1  371.04  5289.2  371.78  5294.3  372.61
    5330  372.59  5335.2  373.46  5361.6  373.27  5534.3  378.37  5578.6  377.59
#Mann= 5 ,-1 , 0
  4190.5     .16       0  4718.7    .033       0  4724.7     .16       0
  4753.3     .05       0  5192.3     .16       0
Bank Sta=4691.9,5212.6
XS Rating Curve= 0 ,0
Exp/Cntr=0.3,0.1

Type RM Length L Ch R = 1 ,28570   ,71,71,71
BEGIN DESCRIPTION:
GUM CREEK 59.0
END DESCRIPTION:
XS GIS Cut Line= 3
      3746793.72     10614423.07      3747793.37     10614640.69
       3747942.5     10614709.72
#Sta/Elev= 30
  4445.8     377  4456.3  376.49  4500.3  379.06  4549.4  379.22  4554.5  378.54
  4582.2  378.14  4615.6  376.96  4686.5  377.16  4740.7  373.85  4748.6   371.9
  4758.9   371.3  4769.1  370.38  4776.3  369.01  4779.1  368.51  4782.3  369.01
  5089.2  369.01  5173.6  369.01  5260.3  369.01  5270.6  369.36  5280.8  370.97
  5311.3  371.72  5392.1  374.02  5424.1   373.1  5474.9  373.55  5486.8  372.99
  5497.8  373.51  5541.9  373.14    5595  374.42  5623.5  373.68  5633.2  374.58
#Mann= 7 ,-1 , 0
  4445.8     .16       0  4582.2     .05       0  4776.3    .033       0
  4782.3     .05       0  5089.2     .16       0  5173.6     .05       0
  5311.3     .16       0
Bank Sta=4758.9,5280.8
XS Rating Curve= 0 ,0
Exp/Cntr=0.3,0.1

Type RM Length L Ch R = 1 ,28499   ,63,63,63
BEGIN DESCRIPTION:
Mapping XS eb83b85d
END DESCRIPTION:
XS GIS Cut Line= 5
      3746765.37     10614477.85      3747185.47     10614573.33
      3747385.12     10614621.94      3747650.75     10614672.29
       3747815.1     10614724.19
#Sta/Elev= 30
  4455.7  374.63  4492.4  374.76  4583.6  378.59    4619   376.9  4669.8  373.98
  4695.6  375.01  4712.9  376.38  4767.7  373.65  4820.1  373.63  4890.4  373.49
  4920.8  375.18  4931.7  374.32  4952.5  375.17  4978.6  373.87  5021.6  374.48
  5105.5  374.59  5110.6  373.16  5156.3  373.93  5186.3  373.22  5215.2  374.19
  5220.3  372.82  5228.9  372.92  5267.5  374.44  5300.1     372  5316.8  371.89
  5319.6  371.39  5322.8  371.89  5324.9   372.2  5384.9  372.73  5534.7  372.58
#Mann= 11 ,-1 , 0
  4455.7     .16       0    4619     .05       0  4695.6     .16       0
  4820.1     .05       0  4920.8     .16       0  5021.6     .05       0
  5156.3     .16       0  5186.3     .05       0  5316.8     .07       0
  5322.8     .05       0  5384.9     .16       0
Bank Sta=5300.1,5324.9
XS Rating Curve= 0 ,0
Exp/Cntr=0.3,0.1

Type RM Length L Ch R = 1 ,28436   ,32,32,32
BEGIN DESCRIPTION:
GUM CREEK 58.0
END DESCRIPTION:
XS GIS Cut Line= 3
      3746764.61      10614561.3       3747723.5     10614738.63
      3747875.34     10614796.67
#Sta/Elev= 30
  4495.7  371.93  4521.6  370.69  4622.4  376.09  4663.5  374.56  4704.2  370.95
  4738.4  371.18  4744.8  372.34  4775.4  371.27  4855.2  363.96  4903.8   360.9
    4955  361.22  4957.3  358.78    4960  358.28  4963.3  358.78  4968.6  360.22
  5008.1  361.32  5019.4  359.53  5054.9   360.7  5071.2  359.96  5171.9  364.96
  5229.9  366.25  5243.2  365.39  5263.5  366.87  5273.7  370.42  5287.9  372.61
  5314.3  371.18  5365.2  372.98  5444.2  373.03  5552.3  371.86  5633.4  373.17
#Mann= 8 ,-1 , 0
  4495.7     .16       0  4855.2     .05       0  4903.8     .16       0
    4955     .12       0  4957.3     .07       0  4963.3     .12       0
  5054.9     .05       0  5444.2     .16       0
Bank Sta=4955,4968.6
XS Rating Curve= 0 ,0
Exp/Cntr=0.3,0.1

Type RM Length L Ch R = 1 ,28404   ,590,590,590
BEGIN DESCRIPTION:
Mapping XS 358a38cf
END DESCRIPTION:
XS GIS Cut Line= 3
      3746745.16     10614586.28      3747675.96     10614761.22
      3747845.43     10614834.41
#Sta/Elev= 30
  4493.8  371.84  4549.2  369.16  4569.6  371.44  4600.7  371.84  4648.1  375.28
  4742.5  369.01  4758.2  370.01  4803.6  368.33  4815.8     366  4895.2  359.72
  4956.2  357.13  4963.4  348.86  4966.1  348.36  4969.4  348.86    4972  349.18
  4986.7  353.56  4996.9  351.97  5017.3  355.76    5072  357.29  5135.9  362.07
    5141  361.09  5188.4  363.72  5193.5  362.08  5230.9  364.15    5246  363.36
    5292  372.48  5386.4  373.02  5479.6   373.8  5573.6  370.71  5625.5  372.25
#Mann= 6 ,-1 , 0
  4493.8     .16       0  4963.4     .07       0  4969.4     .16       0
    4972     .12       0    5072     .05       0  5386.4     .16       0
Bank Sta=4956.2,4986.7
XS Rating Curve= 0 ,0
Exp/Cntr=0.3,0.1

Type RM Length L Ch R = 1 ,27814   ,515,515,515
BEGIN DESCRIPTION:
GUM CREEK 57.0
END DESCRIPTION:
XS GIS Cut Line= 3
      3746237.31     10614718.11      3746795.03     10615052.31
      3747042.45     10615128.27
#Sta/Elev= 30
  4297.8  380.38  4511.1  376.04  4621.2  371.47  4663.4  367.69  4680.3  365.41
  4731.8  362.47  4738.6  359.96    4760  359.47  4775.6  355.83  4781.4  356.93
  4804.3  352.86  4818.3  351.25  4825.1  353.16  4833.9  353.03  4839.7  350.45
  4848.4     352  4855.3  355.21  4892.2  354.55  4906.7  351.23  4913.6  354.67
    4935  355.66  4990.6  354.22  4992.9  347.74  4995.6  347.24  4998.9  347.74
  5028.6  354.61  5088.8  357.22  5141.8  363.08  5182.9  365.43  5206.8  364.86
#Mann= 7 ,-1 , 0
  4297.8     .16       0  4621.2     .12       0  4663.4     .16       0
  4804.3     .12       0  4992.9     .07       0  4998.9     .12       0
  5141.8     .16       0
Bank Sta=4990.6,5028.6
XS Rating Curve= 0 ,0
Exp/Cntr=0.3,0.1

Type RM Length L Ch R = 1 ,27299   ,282,282,282
BEGIN DESCRIPTION:
GUM CREEK 56.0
END DESCRIPTION:
XS GIS Cut Line= 4
      3746139.68     10614937.31      3746465.17     10615126.09
      3746740.77      10615401.7      3747085.22     10615579.34
#Sta/Elev= 30
  4224.2  379.04  4226.2  379.04    4278  376.64  4293.5  377.25  4534.1  370.61
  4542.4  370.29  4655.2  363.47  4684.3  362.29  4691.4  360.28  4719.6  359.96
  4726.7  357.86  4740.9  356.63  4811.6  353.51  4981.3  354.64  4985.9  351.67
  4992.4  351.67  4996.2  348.61  5001.8  349.06  5008.4  347.26  5011.2  346.76
  5014.4  347.26  5018.4  351.93  5033.9  355.35  5056.4  354.16  5123.5     356
  5151.3  351.06  5157.7  353.56  5212.2  356.01  5327.3  366.34  5377.8  368.58
#Mann= 8 ,-1 , 0
  4224.2      .1       0  4226.2     .16       0  4534.1     .12       0
  4542.4     .16       0  4655.2     .12       0  5008.4     .07       0
  5014.4     .12       0  5327.3     .16       0
Bank Sta=4992.4,5018.4
XS Rating Curve= 0 ,0
Exp/Cntr=0.3,0.1

Type RM Length L Ch R = 1 ,27017   ,228,228,228
BEGIN DESCRIPTION:
Mapping XS 7f32df7f
END DESCRIPTION:
XS GIS Cut Line= 3
      3746306.75     10615362.64      3746753.79     10615716.37
      3747129.18     10615633.92
#Sta/Elev= 30
  4714.3  365.49  4764.7  363.83  4779.1  365.49  4793.5   363.1  4799.9  364.67
  4814.3  362.32  4820.7     363  4948.9  353.28  4977.8  350.55  4982.7  345.23
  4985.5  344.73  4988.7  345.23  4998.6  345.71  5006.7   350.3  5049.5  353.35
  5102.6  352.88  5141.3  354.71  5155.7  349.56  5163.8  349.69    5177  355.03
  5203.6  353.66  5219.8  353.87  5287.5  360.32  5385.3  361.33  5429.1  364.14
  5434.2  363.13  5472.9  365.53    5478  364.45    5536  367.44  5668.7   369.8
#Mann= 6 ,-1 , 0
  4714.3      .1       0  4948.9     .12       0  4982.7     .07       0
  4988.7     .12       0  5102.6     .16       0  5203.6     .12       0
Bank Sta=4977.8,5006.7
XS Rating Curve= 0 ,0
Exp/Cntr=0.3,0.1

Type RM Length L Ch R = 1 ,26789   ,479,479,479
BEGIN DESCRIPTION:
GUM CREEK 55.0
END DESCRIPTION:
XS GIS Cut Line= 3
      3746285.03     10615406.02      3746608.39     10616059.25
      3746822.63     10616496.39
#Sta/Elev= 30
  4628.4   364.6  4700.3  365.17  4827.7  361.12    4947  351.56  4956.6   349.8
  4963.9  348.51  4966.5  344.56  4969.2  344.06  4986.3  345.15  4991.9  349.26
  5001.3  348.91  5008.7  346.09  5014.3  351.73  5098.5  351.47  5113.4  353.44
  5120.9  353.51  5143.3  348.06  5157.5  349.44  5163.6  352.36  5179.8  357.83
  5273.7  363.43  5275.1  363.59  5328.3  364.12  5386.6  368.16  5469.7   370.9
  5575.7  372.29  5626.3  371.15  5689.9  372.98  5720.6  373.56  5844.1  376.97
#Mann= 11 ,-1 , 0
  4628.4      .1       0  4827.7     .16       0    4947     .12       0
  5001.3     .16       0  5113.4     .12       0  5163.6     .16       0
  5273.7     .12       0  5275.1     .16       0  5386.6     .05       0
  5689.9     .16       0  5720.6     .05       0
Bank Sta=4956.6,4991.9
XS Rating Curve= 0 ,0
Exp/Cntr=0.3,0.1

Type RM Length L Ch R = 1 ,26310   ,432,432,432
BEGIN DESCRIPTION:
GUM CREEK 54.0
END DESCRIPTION:
XS GIS Cut Line= 3
      3746190.65     10615383.38      3746037.88     10616046.56
      3746407.67     10616438.92
#Sta/Elev= 30
  4633.6  365.63  4681.6  363.56  4791.8  361.57  4814.8  359.21  4845.8  354.89
  4897.1  349.74  4973.2   349.4  4999.5  343.82    5010  345.88  5021.1  350.32
  5063.9   350.8  5092.1  349.41  5133.2  349.52  5163.9  352.42  5225.5  354.73
  5240.3  356.55  5313.4   359.2    5325  358.79  5332.3  359.77  5339.1  358.53
  5424.1   360.5    5431  359.23  5477.6  361.06  5515.9  363.98  5523.2  365.71
  5530.1  364.33  5621.9   369.3  5629.2  370.58  5706.9  375.45  5853.3  382.32
#Mann= 5 ,-1 , 0
  4633.6      .1       0  4814.8     .16       0  4897.1     .13       0
  5063.9     .16       0  5477.6     .05       0
Bank Sta=4973.2,5021.1
XS Rating Curve= 0 ,0
Exp/Cntr=0.3,0.1

Type RM Length L Ch R = 1 ,25878   ,416,416,416
BEGIN DESCRIPTION:
GUM CREEK 53.0
END DESCRIPTION:
XS GIS Cut Line= 3
      3745765.31     10615199.32      3745782.67     10615921.56
      3746400.72     10616464.95
#Sta/Elev= 30
  4527.7  371.09  4588.6  368.08  4638.6  362.99  4648.6  360.83  4698.6   356.8
  4708.6  354.84  4792.9   349.8  4818.7  348.27    4981  347.99  4988.7  347.41
  4995.7  342.52  4998.5  342.02  5008.7  343.55  5018.7  346.56  5028.7  347.47
  5058.7  349.45  5108.7   354.9  5208.8  360.09  5352.9  361.37  5409.8   360.3
    5481     362  5614.2  363.32  5693.5  363.96  5757.1  366.15  5792.2  368.48
  5799.8  367.98  5834.9  370.94  5849.1  371.01  5983.8  379.46  6073.1  382.65
#Mann= 5 ,-1 , 0
  4527.7      .1       0  4792.9     .16       0    4981     .13       0
  5028.7     .16       0  5614.2     .05       0
Bank Sta=4988.7,5018.7
XS Rating Curve= 0 ,0
Exp/Cntr=0.3,0.1

Type RM Length L Ch R = 1 ,25462   ,94,94,94
BEGIN DESCRIPTION:
GUM CREEK 52.0
END DESCRIPTION:
XS GIS Cut Line= 3
      3745363.73      10615449.6      3745787.33     10615947.86
      3746395.97      10616490.5
#Sta/Elev= 30
  4748.6  364.54  4752.9  367.51  4767.2  368.08  4830.9  365.71  4859.5  362.61
  4902.3  354.06  4945.2  347.56  4972.6  347.09  4980.3  345.43  4986.9   346.6
  4998.1  341.38  5000.9  340.88  5004.1  341.38  5008.9  341.42  5015.4  347.46
  5129.7  346.32  5182.9  347.37  5257.1  349.16  5277.9  352.72  5299.9  353.94
  5306.5  356.16  5349.3  358.56  5355.9  360.25  5462.3  361.45  5519.2  359.82
  5639.5  360.73  5722.5  362.81  5880.3  366.08  6064.3  376.47    6218  383.17
#Mann= 5 ,-1 , 0
  4748.6     .12       0  4998.1     .07       0  5004.1     .12       0
  5182.9     .16       0  5722.5     .05       0
Bank Sta=4986.9,5015.4
XS Rating Curve= 0 ,0
Exp/Cntr=0.3,0.1

Type RM Length L Ch R = 1 ,25368   ,236,236,236
BEGIN DESCRIPTION:
Mapping XS 1e91cc61
END DESCRIPTION:
XS GIS Cut Line= 3
      3745247.69     10615503.81      3745694.71     10615911.77
      3746352.26     10616894.84
#Sta/Elev= 30
    4731  354.56  4744.1  349.09  4765.1  350.49  4772.5  353.31  4828.6  352.22
    4836  355.57  4906.9  350.24  4913.7  347.25  4942.1  346.04  4956.3  342.32
  4970.5  344.73  4977.3  341.99  4984.6  346.46  4991.4  345.88  5002.6  341.05
  5005.3  340.55  5008.6  341.05  5027.2  346.98  5048.2  345.46    5140  346.71
  5161.7  344.93    5265  347.27  5331.2  350.99  5395.2  360.18  5431.2  361.54
  5627.9  356.68    6254  374.67  6398.1  373.68  6458.1     370  6518.9  366.23
#Mann= 6 ,-1 , 0
    4731     .12       0  5002.6     .07       0  5008.6     .12       0
    5265     .16       0  5627.9     .05       0  6458.1     .16       0
Bank Sta=4984.6,5027.2
XS Rating Curve= 0 ,0
Exp/Cntr=0.3,0.1

Type RM Length L Ch R = 1 ,25132   ,73,73,73
BEGIN DESCRIPTION:
Mapping XS c8e14d2b
END DESCRIPTION:
XS GIS Cut Line= 3
      3745063.23     10615538.53      3745557.99     10615926.96
      3746254.61      10617051.1
#Sta/Elev= 30
  4428.8  357.93  4479.9  357.54  4590.3  357.38  4724.1  355.51  4818.4  352.46
  4869.2  347.66  4975.6  345.83  4983.6  345.36  4993.4  340.54  4996.2  340.04
  4999.4  340.54    5019   346.4  5062.7  346.56  5104.9  345.88  5142.2   346.8
    5206  354.31  5279.2  355.62  5317.9  353.72  5402.8  352.17    5584  360.87
  5867.6  361.28  6004.6  366.71  6056.6  364.85  6062.5  366.88  6108.6  366.56
  6114.5  368.47  6179.2  366.47  6218.1  360.51  6263.4  363.79  6380.3   363.6
#Mann= 11 ,-1 , 0
  4428.8     .05       0  4479.9     .16       0  4590.3     .05       0
  4724.1     .12       0  4993.4     .07       0  4999.4     .12       0
  5062.7     .05       0  5104.9     .16       0  5317.9     .05       0
  6218.1     .16       0  6263.4     .05       0
Bank Sta=4975.6,5019
XS Rating Curve= 0 ,0
Exp/Cntr=0.3,0.1

Type RM Length L Ch R = 1 ,25059   ,85,85,85
BEGIN DESCRIPTION:
Mapping XS 254b1d8c
END DESCRIPTION:
XS GIS Cut Line= 4
      3745104.91     10615619.12      3745393.13     10615865.67
      3745597.99     10616094.83      3746202.18     10617124.38
#Sta/Elev= 30
  4516.2  360.19  4541.7  360.09  4699.7  356.94    4764   354.9  4988.2  345.56
  5002.4  349.26  5006.1  343.37  5008.9  342.87  5012.1  343.37  5016.6  349.42
  5173.9  347.04  5261.5  349.35  5471.4  351.19  5492.8  355.73  5551.5  351.75
  5557.3  356.78  5567.1  353.22  5572.9  358.81  5580.1  354.21  5594.4  357.04
  5610.1  352.69  5615.9  358.69  5625.8  353.76  5638.1  357.96  5668.7  352.57
  5690.2  356.79  5727.3  352.61  5989.1  360.24  6202.1  356.79  6396.6  365.56
#Mann= 8 ,-1 , 0
  4516.2     .16       0  4541.7     .05       0  4699.7     .08       0
    4764     .05       0  5006.1     .04       0  5012.1     .05       0
  5173.9     .16       0  5261.5     .05       0
Bank Sta=5002.4,5016.6
XS Rating Curve= 0 ,0
Exp/Cntr=0.3,0.1

Type RM Length L Ch R = 1 ,24974   ,149,149,149
BEGIN DESCRIPTION:
GUM CREEK 51.0
END DESCRIPTION:
XS GIS Cut Line= 3
      3745139.14     10615766.35      3745479.86     10616072.36
      3746044.11     10617148.77
#Sta/Elev= 30
  4647.9  370.07  4720.3  368.44  4751.2  364.38  4785.3  362.22  4792.7  358.43
  4835.4  352.97  4972.4  344.23  4984.1  344.19    5002  339.35  5004.8  338.85
    5008  339.35  5019.2   344.1    5076  346.64  5134.6  341.95  5156.7  344.99
  5171.2  342.28  5206.5   343.6  5216.3  346.11  5250.6  343.94  5333.2  347.29
  5355.2  345.14  5526.1  355.35  5608.7  349.63    5719  352.99  5829.3   351.1
  5845.7  353.65  6004.8   354.2  6172.8  358.63  6313.6   365.3  6321.2  365.33
#Mann= 9 ,-1 , 0
  4647.9     .05       0  4720.3     .08       0  4751.2     .12       0
  4972.4     .05       0    5002     .04       0    5008     .05       0
  6004.8     .16       0  6172.8     .05       0  6313.6     .16       0
Bank Sta=4984.1,5019.2
XS Rating Curve= 0 ,0
Exp/Cntr=0.3,0.1

Type RM Length L Ch R = 1 ,24825   ,353,353,353
BEGIN DESCRIPTION:
Mapping XS 7fadc2d1
END DESCRIPTION:
XS GIS Cut Line= 3
      3745108.74     10615905.23       3745462.5     10616189.54
      3745992.01     10617163.92
#Sta/Elev= 30
    4629  372.78  4655.2  371.19  4719.1  365.35  4818.3  350.22  4853.5  347.02
  4882.3  345.36  4931.9  344.86  4960.7  346.42  4981.5  344.93  4999.3  338.58
  5002.1  338.08  5005.3  338.58  5010.3  345.67  5016.7  346.17  5038.8  346.29
  5074.3  344.42    5151  344.72  5235.5  346.16  5317.3  345.05  5366.2  347.18
  5404.7  348.78  5595.7  349.62  5753.4  355.61  5833.4  356.36  5928.2  357.57
  5966.2  360.29  5988.1  359.63  6026.1  362.45  6164.2  366.39  6191.8  366.44
#Mann= 9 ,-1 , 0
    4629     .05       0  4655.2     .12       0  4999.3     .07       0
  5005.3     .12       0  5038.8     .05       0    5151     .12       0
  5366.2     .05       0  5833.4     .16       0  6164.2     .05       0
Bank Sta=4981.5,5016.7
XS Rating Curve= 0 ,0
Exp/Cntr=0.3,0.1

Type RM Length L Ch R = 1 ,24472   ,461,461,461
BEGIN DESCRIPTION:
GUM CREEK 50.0
END DESCRIPTION:
XS GIS Cut Line= 3
      3744918.76     10616086.28      3745331.95      10616534.2
      3746033.21      10617315.3
#Sta/Elev= 30
  4627.6  375.14  4659.5  371.49  4673.7  367.82  4694.1  366.31  4715.7   360.8
  4747.2  355.79  4836.5  346.99  4914.1  343.65  4977.6  344.45    4985  342.41
  4991.8  341.41  4996.2  338.08  4998.9  337.58  5002.2  338.08    5006  338.13
  5013.4   342.5  5020.2  338.55  5027.5  345.07  5030.4  345.41  5147.8  343.62
  5268.1   344.3  5317.4  346.16  5480.3  357.47  5629.1  358.25  5671.7  359.31
  5678.4  360.97  5701.9  360.58  5919.1  364.99  6045.1  365.93  6286.7  371.23
#Mann= 7 ,-1 , 0
  4627.6     .05       0  4747.2     .12       0  4996.2     .07       0
  5002.2     .12       0  5030.4     .05       0  5701.9     .16       0
  6045.1     .05       0
Bank Sta=4985,5013.4
XS Rating Curve= 0 ,0
Exp/Cntr=0.3,0.1

Type RM Length L Ch R = 1 ,24011   ,462,462,462
BEGIN DESCRIPTION:
GUM CREEK 49.0
END DESCRIPTION:
XS GIS Cut Line= 4
      3744739.91     10616333.23      3744963.89     10616621.46
      3745500.35     10616779.44      3746031.58     10617394.01
#Sta/Elev= 30
  4680.4  365.89  4777.9  362.14  4913.1  347.46  4942.5  345.34  4955.2  341.98
  4963.3  341.27  4969.6  342.65  4984.1  342.97  4995.6  338.97  4998.3  338.47
  5001.6  338.97  5005.8  339.09  5013.1  343.59  5041.4  342.35  5113.9  343.43
  5169.8  342.59  5306.6  343.58  5445.2  351.46    5583  356.83  5719.9  357.78
  5817.1  360.41  5895.8  360.79  5902.4  361.93  5959.4  360.75  5980.3  362.31
    6080  363.21  6114.1  365.52  6313.7  369.61  6334.6  371.45    6417  374.16
#Mann= 7 ,-1 , 0
  4680.4     .05       0  4913.1     .12       0  4995.6     .07       0
  5001.6     .12       0  5169.8     .05       0  5719.9     .16       0
  6114.1     .05       0
Bank Sta=4984.1,5013.1
XS Rating Curve= 0 ,0
Exp/Cntr=0.3,0.1

Type RM Length L Ch R = 1 ,23549   ,503,503,503
BEGIN DESCRIPTION:
GUM CREEK 48.0
END DESCRIPTION:
XS GIS Cut Line= 3
      3744599.61     10616560.19      3744649.61     10616910.19
      3744949.64     10617310.22
#Sta/Elev= 30
  4659.6  358.69  4740.4  355.24  4766.1  352.37    4801  350.43  4831.3  346.38
  4871.7  342.97  4912.1  341.47  4962.6  341.52  4982.9  342.62    4993  337.57
  5000.1  335.99  5002.8  335.49  5006.1  335.99  5010.6  341.53  5026.7  343.28
    5035  342.31  5126.7  340.41  5170.4  340.43    5260  342.52  5291.3  344.39
  5337.4  350.29  5363.2  351.68  5370.4  353.41  5391.3  354.68  5420.4  358.16
  5426.7  357.25    5435  359.07  5494.2  364.19  5495.1  364.27  5513.2  365.86
#Mann= 8 ,-1 , 0
  4659.6     .05       0  4766.1     .12       0  5000.1     .07       0
  5006.1     .12       0    5260     .16       0  5337.4     .12       0
  5494.2     .16       0  5495.1     .12       0
Bank Sta=4982.9,5010.6
XS Rating Curve= 0 ,0
Exp/Cntr=0.3,0.1

Type RM Length L Ch R = 1 ,23046   ,328,328,328
BEGIN DESCRIPTION:
GUM CREEK 47.0
END DESCRIPTION:
XS GIS Cut Line= 3
      3744099.62     10617060.19      3744399.61     10617210.19
      3744599.63     10617510.23
#Sta/Elev= 30
  4656.6  355.32  4678.9  355.14  4723.7   352.3  4768.4  346.25  4849.4  338.72
    4978  341.39  4982.4  340.82  4983.6  340.66  4986.2  333.72    4989  333.22
  4992.2  333.72    4995  333.72  4999.5   336.2  5005.5  341.52  5071.6     341
  5077.6  340.78  5086.6   338.9  5092.7  339.98  5107.7  338.87  5122.7  339.14
  5143.7  341.24  5149.7  343.34  5158.8  342.94  5179.8  346.57  5185.8  345.98
  5200.8  347.23  5215.8  349.44  5257.9  353.15  5272.9  355.82  5352.6   362.3
#Mann= 4 ,-1 , 0
  4656.6     .05       0  4982.4     .12       0  4986.2     .07       0
  4992.2     .12       0
Bank Sta=4983.6,5005.5
XS Rating Curve= 0 ,0
Exp/Cntr=0.3,0.1

Type RM Length L Ch R = 1 ,22718   ,863,863,863
BEGIN DESCRIPTION:
GUM CREEK 46.0
END DESCRIPTION:
XS GIS Cut Line= 3
      3744049.63     10617110.23      3744249.61     10617410.19
      3744549.63     10617710.21
#Sta/Elev= 30
  4559.5  355.63    4582  355.28  4631.6  351.37  4645.1  349.24  4654.1  349.18
  4739.7  339.08  4762.3   338.2  4840.4  339.09  4847.9  336.39  4857.5  332.54
  4858.4  332.43  4861.2  331.93  4864.4  332.43  4876.4  334.16    4884  333.15
  4891.5  333.81  4897.5  338.72  4906.5  339.35  4976.6     340  5004.9  336.58
    5019   339.5  5061.4  339.67  5132.1  345.32  5146.3  345.47  5174.6  347.81
  5231.1  355.16  5245.3  358.14  5308.5  366.71  5330.1  368.59  5344.3   368.5
#Mann= 5 ,-1 , 0
  4559.5     .05       0  4857.5     .12       0  4858.4     .07       0
  4864.4     .12       0  5308.5     .05       0
Bank Sta=4847.9,4876.4
XS Rating Curve= 0 ,0
Exp/Cntr=0.3,0.1

Type RM Length L Ch R = 1 ,21855   ,702,702,702
BEGIN DESCRIPTION:
GUM CREEK 45.0
END DESCRIPTION:
XS GIS Cut Line= 2
      3743845.84     10617145.33      3743897.93     10618259.91
#Sta/Elev= 30
  4413.2  353.97  4448.1  353.38  4558.2  347.65  4588.3  347.69  4602.1  349.24
  4648.3  349.43  4688.4  346.28  4768.3  342.25  4814.4  340.88  4819.4  342.25
  4898.6  337.05  4978.7  338.02  4988.7  335.81  4995.7  331.43  4998.5  330.93
  5001.7  331.43  5008.7  332.55  5018.7  337.49  5048.8   337.1  5068.8  338.05
  5118.8  336.33  5138.9   337.6  5168.9   336.9  5178.9  335.19  5188.9  336.64
  5243.8  335.32  5312.7  338.48  5399.1  342.44  5499.2  351.34    5529  355.15
#Mann= 5 ,-1 , 0
  4413.2     .05       0  4768.3     .12       0  4995.7     .07       0
  5001.7     .12       0  5312.7     .05       0
Bank Sta=4978.7,5018.7
XS Rating Curve= 0 ,0
Exp/Cntr=0.3,0.1

Type RM Length L Ch R = 1 ,21153   ,445,445,445
BEGIN DESCRIPTION:
GUM CREEK 44.0
END DESCRIPTION:
XS GIS Cut Line= 3
      3743453.48      10616895.3      3743384.04      10617534.2
      3743384.04     10618141.83
#Sta/Elev= 30
  4300.6  354.24  4386.9  350.53  4466.5   344.4  4473.4     343  4506.7  342.03
  4526.8   341.5  4536.9  339.76  4546.2   339.9  4687.8  334.28  4745.6  333.39
  4788.3  332.79  4939.2  333.65  4979.3  334.38  4989.3  333.11  4996.3  329.71
    4999  329.21  5002.3  329.71  5009.3  334.46  5037.2  334.34  5089.3  334.95
  5219.3  342.79  5279.3  343.68  5309.3  344.88  5319.3  346.33  5331.4  345.77
  5339.3  345.26  5349.3  346.64  5399.9  347.81  5499.3  352.47  5550.9  356.14
#Mann= 10 ,-1 , 0
  4300.6     .16       0  4506.7     .05       0  4546.2     .16       0
  4745.6     .05       0  4939.2     .12       0  4996.3     .07       0
  5002.3     .12       0  5037.2     .16       0  5331.4     .12       0
  5399.9     .05       0
Bank Sta=4979.3,5009.3
XS Rating Curve= 0 ,0
Exp/Cntr=0.3,0.1

Type RM Length L Ch R = 1 ,20708   ,508,508,508
BEGIN DESCRIPTION:
GUM CREEK 43.0
END DESCRIPTION:
XS GIS Cut Line= 3
       3742649.6     10616760.18      3742999.61     10617560.19
      3743299.61     10618310.19
#Sta/Elev= 30
  4131.2  374.26  4229.4   367.2    4268  363.41  4343.7  359.92  4541.7   341.8
    4677  335.98  4709.7  332.47  4721.8  332.59  4731.5  330.95  4884.4   330.9
    4891  333.18  4906.2  333.54  4914.4  331.61  4938.5     331  4982.6  331.64
  4992.5  326.66  4995.2  326.16  4998.5  326.66  5001.7  331.93  5013.8   332.5
  5019.2  328.26    5026  330.71  5036.7   332.6  5067.7  331.24  5119.2  331.27
  5241.4  336.88  5283.1  337.03  5489.1  344.99  5606.2  353.71  5812.2  364.62
#Mann= 5 ,-1 , 0
  4131.2     .05       0  4938.5     .12       0  4992.5     .07       0
  4998.5     .12       0  5119.2     .05       0
Bank Sta=4982.6,5001.7
XS Rating Curve= 0 ,0
Exp/Cntr=0.3,0.1
