HEC-RAS study KEECHIE CREEK.prj: KEECHIE CREEK Base Level Engineering

--- KEECHIE CREEK.g01 (geometry) --- (continued)

Type RM Length L Ch R = 1 ,64098   ,395,395,395
BEGIN DESCRIPTION:
KEECHIE CREEK 95.0
END DESCRIPTION:
XS GIS Cut Line= 3
      3725528.38     10647394.47      3723978.91     10646951.76
      3723206.37      10646825.9
#Sta/Elev= 30
  3183.6  328.28  3244.7  323.61  3296.7  316.45  3356.6  312.69  3548.3  298.37
  3615.9  291.22  3733.5   285.9  4149.5  281.87  4198.3  280.17  4367.9  283.05
    4901  282.72  4960.9  284.25  4976.7  274.73    4994  271.72  4996.8  271.22
    5000  271.72  5017.3  277.82  5022.4  284.66  5078.1  287.38  5083.9  289.15
  5138.9  293.65  5145.4  295.76  5273.5  307.61  5396.4  320.01  5402.3  322.35
  5452.9  324.93  5483.3  329.87  5493.5  329.15    5534  334.41  5577.8  336.54
#Mann= 6 ,-1 , 0
  3183.6     .12       0  3356.6     .05       0    4901     .12       0
    4994     .07       0    5000     .12       0  5273.5     .16       0
Bank Sta=4960.9,5022.4
XS Rating Curve= 0 ,0
Exp/Cntr=0.3,0.1

Type RM Length L Ch R = 1 ,63703   ,515,515,515
BEGIN DESCRIPTION:
KEECHIE CREEK 94.0
END DESCRIPTION:
XS GIS Cut Line= 3
      3725499.59     10646460.19      3723949.61     10646560.19
      3723549.63     10646510.19
#Sta/Elev= 30
  3410.1  334.06  3460.2  325.22  3491.5   322.3  3500.3  318.94  3560.4  308.98
  3716.1  289.11  3750.8  285.88    3871  281.38  4412.2  279.79  4418.4  281.44
  4438.1  281.24  4446.6  280.94  4892.5  281.48  4965.8  283.02  4983.5  273.07
  4998.1  271.36  5000.8  270.86  5004.1  271.36  5013.7  273.39  5023.8   280.6
  5033.8  282.69  5081.7  281.52  5124.5  288.12  5134.6  294.71  5162.3  306.91
  5167.4  311.66    5185  317.88  5207.2   323.1  5255.6  330.88  5366.4  333.14
#Mann= 8 ,-1 , 0
  3410.1     .12       0  3716.1     .05       0  4438.1     .12       0
  4446.6     .05       0  4892.5     .12       0  4998.1     .07       0
  5004.1     .12       0  5207.2     .16       0
Bank Sta=4965.8,5033.8
XS Rating Curve= 0 ,0
Exp/Cntr=0.3,0.1

Type RM Length L Ch R = 1 ,63188   ,1116,1116,1116
BEGIN DESCRIPTION:
KEECHIE CREEK 93.0
END DESCRIPTION:
XS GIS Cut Line= 3
      3725649.57     10646310.18      3724099.61     10646110.19
       3723649.6     10646210.19
#Sta/Elev= 30
  3418.3  341.98    3509  337.08  3549.3  329.64  3680.4  311.42  3693.6  310.88
    3872  288.87  3915.6  285.71  4001.2     281  4073.6  279.79  4574.1  280.06
    4598  280.53  4618.1   276.4  4626.3  279.83  4636.8   279.9  4668.5  279.02
  4889.8  281.21  4943.9  281.72  4960.9  278.61  4978.6  272.23  5002.4  270.58
  5005.2  270.08  5008.4  270.58  5022.1  281.54  5073.3  281.95  5124.5  287.45
  5175.7  290.51  5257.7  299.03  5276.9  299.58  5437.3  321.44  5442.1  321.99
#Mann= 8 ,-1 , 0
  3418.3     .12       0  3915.6     .05       0  4574.1     .12       0
  4636.8     .05       0  4889.8     .12       0  5002.4     .07       0
  5008.4     .12       0  5437.3     .16       0
Bank Sta=4943.9,5022.1
XS Rating Curve= 0 ,0
Exp/Cntr=0.3,0.1

Type RM Length L Ch R = 1 ,62072   ,465,465,465
BEGIN DESCRIPTION:
KEECHIE CREEK 92.0
END DESCRIPTION:
XS GIS Cut Line= 3
      3724699.61     10645010.19      3724349.61     10645210.19
       3723549.6      10646010.2
#Sta/Elev= 30
  4599.2  331.19  4693.5  321.55  4709.3  317.25  4752.5  310.93  4805.8  299.58
  4864.1  291.63  4870.6   287.9  4876.3  289.03  4886.4  286.19  4898.7  285.41
    4908  279.77  4913.8  278.08  4972.8  280.13  4999.4  269.26  5013.5  269.19
  5016.2  268.69  5019.5  269.19  5030.6  270.59  5044.7  279.16  5186.2  277.22
  5231.1  278.19  5454.9  276.73  5511.4  278.43  5633.9  277.65    5766  277.13
  5836.7  281.02    5865  285.61  6104.4  314.26    6129  318.79  6133.7  318.97
#Mann= 7 ,-1 , 0
  4599.2     .12       0  5013.5     .07       0  5019.5     .12       0
  5231.1     .07       0  5633.9     .12       0  6104.4     .16       0
    6129     .12       0
Bank Sta=4972.8,5044.7
XS Rating Curve= 0 ,0
Exp/Cntr=0.3,0.1

Type RM Length L Ch R = 1 ,61607   ,589,589,589
BEGIN DESCRIPTION:
KEECHIE CREEK 91.0
END DESCRIPTION:
XS GIS Cut Line= 3
      3724649.65     10644860.17      3724049.61     10645160.19
      3723299.59     10645860.21
#Sta/Elev= 30
  4353.1  328.09  4425.1  322.61  4518.1  308.66    4546  306.33  4562.8  301.11
  4568.4  301.74  4613.1   295.1  4650.7  287.97  4680.2  283.98  4696.9  279.45
  4724.9  277.74    4764  281.49  4786.4  279.35  4965.3  278.12    5007  268.39
  5009.7  267.89    5013  268.39  5015.6  268.77  5021.2  274.21  5027.4  274.21
    5031  277.36  5037.9  279.31  5158.6  276.28  5236.2  278.06  5427.2  275.89
  5519.1  275.99  5604.1  278.77  5780.9  299.71  6007.6  332.24  6049.9  335.59
#Mann= 5 ,-1 , 0
  4353.1     .12       0  4425.1     .16       0  4650.7     .12       0
    5007     .07       0    5013     .12       0
Bank Sta=4965.3,5037.9
XS Rating Curve= 0 ,0
Exp/Cntr=0.3,0.1

Type RM Length L Ch R = 1 ,61018   ,587,587,587
BEGIN DESCRIPTION:
KEECHIE CREEK 90.0
END DESCRIPTION:
XS GIS Cut Line= 3
      3724549.57     10644860.18      3723749.61     10644760.19
      3723049.65     10645210.16
#Sta/Elev= 30
  4181.8  317.25    4212  313.33  4272.5  301.15  4343.2  292.16  4385.8  286.61
  4403.5  281.84  4433.7  280.02  4461.4  276.31  4541.7  277.28  4640.9  276.62
  4740.1  275.33  4839.4  277.11  4967.8  278.14  4977.9  274.15  4985.5  268.62
  4992.6  267.91  4995.3  267.41  4998.6  267.91  5010.8  268.31  5023.6  277.27
  5031.9   278.1  5219.5  274.32  5494.9  275.41  5582.4  285.98  5594.6  290.51
  5646.1  294.93  5712.8   303.8    5725  307.63  5748.8  311.37  5820.1  319.98
#Mann= 8 ,-1 , 0
  4181.8     .16       0  4343.2     .12       0  4541.7     .07       0
  4640.9     .12       0  4740.1     .07       0  4839.4     .12       0
  4992.6     .07       0  4998.6     .12       0
Bank Sta=4967.8,5031.9
XS Rating Curve= 0 ,0
Exp/Cntr=0.3,0.1

Type RM Length L Ch R = 1 ,60431   ,548,548,548
BEGIN DESCRIPTION:
KEECHIE CREEK 89.0
END DESCRIPTION:
XS GIS Cut Line= 3
       3724899.6     10644510.19      3723499.61     10644310.19
       3722799.6     10644460.19
#Sta/Elev= 30
  3570.2  341.26  3616.7  338.22  3741.9  323.84    3752  320.36  3802.5  314.57
  3842.9  305.42  3921.3  294.04  4014.7  281.06  4113.1  275.38    4439  275.32
  4607.5  273.51  4954.1  276.88  4974.3  267.92  5006.1   267.3  5008.9   266.8
  5012.1   267.3  5025.3  267.73  5035.5  276.68  5311.7  272.85  5475.3   292.3
    5483  299.27  5488.1  293.67  5495.8  298.18  5516.2  296.38  5581.8  305.21
  5618.5  312.64  5626.1  316.95  5631.3  312.81  5638.9   315.6  5700.3  319.02
#Mann= 8 ,-1 , 0
  3570.2     .05       0  3616.7     .12       0  3921.3     .07       0
  4113.1     .12       0    4439     .07       0  4607.5     .12       0
  5006.1     .07       0  5012.1     .12       0
Bank Sta=4954.1,5035.5
XS Rating Curve= 0 ,0
Exp/Cntr=0.3,0.1

Type RM Length L Ch R = 1 ,59883   ,514,514,514
BEGIN DESCRIPTION:
KEECHIE CREEK 88.0
END DESCRIPTION:
XS GIS Cut Line= 3
      3724649.61     10643210.19      3723249.61     10643910.19
      3722749.58      10644110.2
#Sta/Elev= 30
  3404.3  335.06  3457.4  335.07  3493.7   331.6  3753.7     288  3932.6  271.86
  3971.7  271.64  3994.1  275.47  4038.8   271.8  4282.5  273.42  4757.2  273.77
    4870  274.61  4920.3  275.06    4979  276.26  4998.9  267.04  5001.6  266.54
  5004.9  267.04    5014  267.47  5023.4  274.62  5038.2  275.26  5116.3  273.32
  5140.5   276.6  5145.9  281.76    5185  280.52    5224  288.55  5248.2  287.18
    5325  296.45  5337.1  300.79  5346.5  298.65    5469  312.66  5508.1  314.16
#Mann= 7 ,-1 , 0
  3404.3     .12       0  4282.5     .07       0  4757.2     .12       0
    4870     .07       0  4920.3     .12       0  4998.9     .07       0
  5004.9     .12       0
Bank Sta=4979,5038.2
XS Rating Curve= 0 ,0
Exp/Cntr=0.3,0.1

Type RM Length L Ch R = 1 ,59369   ,582,582,582
BEGIN DESCRIPTION:
KEECHIE CREEK 87.0
END DESCRIPTION:
XS GIS Cut Line= 3
      3723999.63     10642710.16      3723199.61     10643510.19
      3722699.63     10644110.17
#Sta/Elev= 30
  3852.3  296.21  3931.9  289.61  4092.8  277.53    4121  278.88  4234.2  272.36
  4517.9  271.99  4782.2  272.75  4969.6  274.32  4980.2  269.24  4990.9  270.59
  4994.4  266.17  4997.1  265.67  5000.4  266.17  5011.7  267.91  5019.5  273.32
    5026  274.65  5161.4  274.96  5167.9  278.01  5239.5  278.28    5246  282.14
  5253.8  280.45  5274.6  283.24  5374.2   282.1  5438.7  285.49  5508.9  289.74
  5530.4  295.33  5601.4  300.04  5608.5  302.78  5636.5  303.39  5764.7  316.73
#Mann= 6 ,-1 , 0
  3852.3     .16       0  3931.9     .12       0  4517.9     .07       0
  4782.2     .12       0  4994.4     .07       0  5000.4     .12       0
Bank Sta=4969.6,5026
XS Rating Curve= 0 ,0
Exp/Cntr=0.3,0.1

Type RM Length L Ch R = 1 ,58787   ,580,580,580
BEGIN DESCRIPTION:
KEECHIE CREEK 86.0
END DESCRIPTION:
XS GIS Cut Line= 3
      3723649.63     10642260.16      3723099.61     10643060.19
      3722399.62     10644310.17
#Sta/Elev= 30
  4041.4  310.77  4099.6  308.16  4137.1  303.76  4164.5  299.42  4228.2  289.89
  4235.6  286.59    4264  281.59  4322.1  274.34  4380.4  270.28  4766.8  270.69
  4841.2  271.64    4969  273.45  4983.9  268.18  5001.8   265.7  5004.6   265.2
  5007.8   265.7  5015.1  265.95  5020.2  273.46  5652.7  270.68  5701.8  271.85
  5804.5  281.72  5866.1  284.54  5940.7  291.84    5968   294.1    6107  306.43
  6296.5  317.42  6306.8  321.13  6312.5  318.67  6334.2  319.59  6444.9  328.06
#Mann= 11 ,-1 , 0
  4041.4     .16       0  4137.1     .12       0  4164.5     .16       0
  4322.1     .12       0  4766.8     .07       0  4841.2     .12       0
  5001.8     .07       0  5007.8     .12       0  5866.1     .16       0
  5940.7      .1       0    5968     .12       0
Bank Sta=4969,5020.2
XS Rating Curve= 0 ,0
Exp/Cntr=0.3,0.1

Type RM Length L Ch R = 1 ,58207   ,556,556,556
BEGIN DESCRIPTION:
KEECHIE CREEK 85.0
END DESCRIPTION:
XS GIS Cut Line= 3
      3723449.63     10642160.17      3722649.61     10642760.19
      3721849.61     10643560.19
#Sta/Elev= 30
  3986.1  301.16  3998.3  297.72    4142  283.16  4171.6  281.54    4208  278.79
  4297.5  276.47  4472.6  269.84  4722.2  269.84  4964.2  272.42  4972.6  271.63
  4978.8   267.7  4982.4  268.11  4989.7  268.18  4997.3  265.21    5000  264.71
  5003.3  265.21  5014.4     270  5028.6  272.34  5085.1  270.13  5184.1  271.23
  5226.5  269.14  5283.1  271.16  5424.5  268.66    5467  269.78  5919.5  268.98
  5976.1  273.28  6046.8  283.62  6075.1  285.78  6103.4  291.02  6117.5  291.65
#Mann= 9 ,-1 , 0
  3986.1     .12       0  3998.3     .16       0    4142     .05       0
  4171.6      .1       0  4297.5     .12       0  4722.2     .07       0
  4982.4     .12       0  4997.3     .07       0  5003.3     .12       0
Bank Sta=4964.2,5028.6
XS Rating Curve= 0 ,0
Exp/Cntr=0.3,0.1

Type RM Length L Ch R = 1 ,57651   ,525,525,525
BEGIN DESCRIPTION:
KEECHIE CREEK 84.0
END DESCRIPTION:
XS GIS Cut Line= 3
      3722299.61     10641710.17      3722299.61     10642410.19
       3721599.6     10643660.21
#Sta/Elev= 30
  4283.7  300.75  4323.7  300.05  4464.3  291.16  4573.7  283.68  4713.7     270
  4823.7  268.59  4973.7  271.18  4978.2  264.88    4981  264.38  4984.2  264.88
  4997.4  264.88  5013.4  271.42  5019.1   271.7  5305.7  268.68    5381   270.1
  5533.9  268.69  5556.8  270.34  5878.7  269.23  5969.4   275.6  5981.5  278.68
  5991.7  277.75  6121.9  292.42  6143.6  297.23  6165.3  296.65  6187.2  298.89
  6246.3  307.89  6262.3  308.22  6343.3  318.88    6349     322  6416.4  328.84
#Mann= 4 ,-1 , 0
  4283.7     .05       0  4464.3     .12       0  4978.2     .07       0
  4984.2     .12       0
Bank Sta=4973.7,5019.1
XS Rating Curve= 0 ,0
Exp/Cntr=0.3,0.1

Type RM Length L Ch R = 1 ,57126   ,563,563,563
BEGIN DESCRIPTION:
KEECHIE CREEK 83.0
END DESCRIPTION:
XS GIS Cut Line= 3
      3722249.63     10641760.17      3721949.61     10642060.19
      3721549.61     10643460.18
#Sta/Elev= 30
  4583.3  298.14  4696.5  292.24  4767.2  286.14  4809.6  280.03  4851.7  277.33
  4936.9  267.61    4951  267.41  4965.2  270.27  4990.4  265.33  4993.2  264.83
  4996.4  265.33  5004.1  270.86  5153.2  268.33  5402.8  268.19  5461.3  268.93
  5475.6  270.94  5567.9  268.53  5631.6  270.34  5652.4  268.37  5808.4  270.14
  5964.4  269.07  6037.2  274.25  6048.9  277.34  6172.4  288.97  6223.1  291.56
  6267.3  297.92  6295.9  299.83  6307.6  303.76  6334.9  304.09  6463.6  321.84
#Mann= 4 ,-1 , 0
  4583.3     .05       0  4851.7     .12       0  4990.4     .07       0
  4996.4     .12       0
Bank Sta=4965.2,5004.1
XS Rating Curve= 0 ,0
Exp/Cntr=0.3,0.1

Type RM Length L Ch R = 1 ,56563   ,140,140,140
BEGIN DESCRIPTION:
Mapping XS 48e77314
END DESCRIPTION:
XS GIS Cut Line= 3
      3721974.51      10641275.8      3721302.64     10641989.34
      3720479.74     10642749.73
#Sta/Elev= 30
  4241.2  294.85  4706.7   278.2  4792.6  276.63  4898.6   267.9  4976.2  269.68
  4983.5  268.03  4987.4  264.03  4990.2  263.53  4993.4  264.03  5004.6  264.54
  5011.9  269.51  5125.2  267.43  5344.5  269.98    5387   268.3  5401.2  269.92
  5519.2  268.98  5598.5  269.28  5736.5  269.51  5762.2  269.24  5876.2  269.33
  5900.9  269.59  5960.2   269.3  6015.9  276.23  6039.6   278.7  6155.6  292.11
  6178.3  295.91  6264.2  310.22  6295.3   313.5    6317  316.17  6341.7  317.94
#Mann= 16 ,-1 , 0
  4241.2     .05       0  4706.7     .12       0  4987.4     .07       0
  4993.4     .12       0  5519.2     .05       0  5598.5     .12       0
  5736.5     .05       0  5762.2     .12       0  5876.2     .05       0
  5900.9     .12       0  6015.9     .05       0  6039.6     .12       0
  6155.6     .05       0  6178.3     .12       0  6295.3     .16       0
    6317     .12       0
Bank Sta=4976.2,5011.9
XS Rating Curve= 0 ,0
Exp/Cntr=0.3,0.1

Type RM Length L Ch R = 1 ,56423   ,204,204,204
BEGIN DESCRIPTION:
KEECHIE CREEK 82.0
END DESCRIPTION:
XS GIS Cut Line= 3
        3721912.     10641228.93      3721162.01     10641942.46
      3720427.66     10642702.86
#Sta/Elev= 30
  4183.9  294.23  4434.2  284.17  4646.2  278.56  4759.4  270.79  4879.5   267.9
  4949.4  269.15  4971.7  268.91  4978.6  264.28  4982.9  263.74  4985.6  263.24
  4988.9  263.74    5000  264.09  5021.1  269.74  5112.6  267.69  5126.5  267.43
  5233.3  267.57  5261.6  269.66  5275.7  269.07  5282.9  266.69    5304  266.14
  5311.2  268.43  5862.8  269.56  5990.1  281.55  6025.3  287.97  6060.8  289.71
  6181.5  306.41  6202.3  310.47  6237.6  313.21  6258.7  316.63  6276.2  316.51
#Mann= 7 ,-1 , 0
  4183.9     .05       0  4949.4     .12       0  4982.9     .07       0
  4988.9     .12       0  5112.6     .08       0  5126.5     .05       0
  6181.5     .16       0
Bank Sta=4971.7,5021.1
XS Rating Curve= 0 ,0
Exp/Cntr=0.3,0.1

Type RM Length L Ch R = 1 ,56219   ,126,126,126
BEGIN DESCRIPTION:
KEECHIE CREEK 81.0
END DESCRIPTION:
XS GIS Cut Line= 3
      3721781.81     10641088.29      3721021.39     10641874.75
       3720319.4     10642566.34
#Sta/Elev= 30
  4045.2  297.95  4421.5  283.77  4663.3  274.27  4712.9  270.58  4870.6  267.63
  4961.5  269.25  4981.5  268.48  4988.7   265.9  5009.8  264.24  5031.2  268.75
  5123.3  267.93  5250.4  267.18  5282.7  264.11  5285.4  263.61  5288.7  264.11
  5299.8  266.98  5321.1  268.18  5328.1   265.8  5335.2  267.48  5589.8  266.26
  5674.7   266.5  5738.3   269.1  5787.7  273.69  5794.8  276.16  5844.3  282.57
    5915   286.9  5985.7  295.16  5992.8   297.9  6042.3  300.07  6124.6  310.07
#Mann= 7 ,-1 , 0
  4045.2     .05       0  4421.5     .12       0  4870.6     .08       0
  4961.5     .07       0  5123.3     .12       0  5282.7     .07       0
  5288.7     .12       0
Bank Sta=4981.5,5031.2
XS Rating Curve= 0 ,0
Exp/Cntr=0.3,0.1

Type RM Length L Ch R = 1 ,56093   ,603,603,603
BEGIN DESCRIPTION:
Mapping XS 7eb6a70d
END DESCRIPTION:
XS GIS Cut Line= 3
      3721635.99     10641036.18      3720917.22     10641833.09
      3720271.41     10642494.52
#Sta/Elev= 30
  4155.3  303.44  4367.9  292.94  4410.5  289.37  4431.4  290.14    4545  281.89
  4622.8  278.81  4785.7  273.85  4899.3  266.94  4983.7  268.57  4991.2  267.54
  4997.9  264.52  5005.4  264.31  5019.6  264.97  5026.3  269.13  5062.7  268.38
  5172.5  267.52  5330.8   267.1  5370.3  263.91    5373  263.41  5376.3  263.91
  5394.4  266.87  5670.3  265.53  5783.5  268.29    5854  275.02  5910.6  283.06
  5967.2  286.65  6002.6  291.74  6108.6  302.71  6115.8  302.08  6152.9  307.68
#Mann= 6 ,-1 , 0
  4155.3     .05       0  4622.8     .12       0  5062.7     .07       0
  5172.5     .12       0  5370.3     .07       0  5376.3     .12       0
Bank Sta=5330.8,5394.4
XS Rating Curve= 0 ,0
Exp/Cntr=0.3,0.1

Type RM Length L Ch R = 1 ,55490   ,1106,1106,1106
BEGIN DESCRIPTION:
KEECHIE CREEK 80.0
END DESCRIPTION:
XS GIS Cut Line= 3
      3721299.65     10641060.16      3720649.61     10641460.19
      3720149.59     10642260.22
#Sta/Elev= 30
  4220.3  299.13  4249.3   298.5  4359.4  291.16  4475.4  281.96  4579.8  277.63
  4707.3  271.76  4765.2  266.58  4896.6  266.41    4970  268.07  4986.5  265.97
  4994.1  263.51  4996.9  263.01  5000.1  263.51  5006.6  266.77  5018.9  267.87
  5085.6  266.93  5106.8  268.02  5158.7  265.21  5164.6  266.41  5172.2  265.01
  5179.9  266.21  5274.2  264.77  5419.9  266.33  5426.4  264.61  5447.6   266.1
  5620.9  264.48  5666.9  266.98  5688.2  271.24  5788.4  284.03    5927  299.26
#Mann= 4 ,-1 , 0
  4220.3     .05       0  4579.8     .12       0  4994.1     .07       0
  5000.1     .12       0
Bank Sta=4970,5018.9
XS Rating Curve= 0 ,0
Exp/Cntr=0.3,0.1

Type RM Length L Ch R = 1 ,54384   ,265,265,265
BEGIN DESCRIPTION:
KEECHIE CREEK 79.0
END DESCRIPTION:
XS GIS Cut Line= 3
      3720749.64     10639960.16      3720099.61     10640660.19
       3719699.6     10642210.21
#Sta/Elev= 30
  4051.9  290.47  4129.9  290.25  4186.6  285.13  4193.4  282.95  4250.1  275.71
  4292.6  272.66    4427  272.61  4603.8  267.78  4788.1  265.51  4922.4  265.04
  4964.9  266.37  4985.9   265.8  4993.3  262.96  5009.8  263.59  5017.5   266.4
  5193.1  264.23  5830.4  262.78  5833.2  262.28  5836.4  262.78  5998.6  264.46
  6066.7  267.18  6188.7  268.96  6264.9   274.1  6305.6  278.77  6380.8  282.81
  6476.1  293.45  6503.7  295.28    6515  297.88  6597.6  303.94    6608  302.57
#Mann= 4 ,-1 , 0
  4051.9     .12       0  5830.4     .07       0  5836.4     .12       0
  6476.1     .16       0
Bank Sta=4964.9,5017.5
XS Rating Curve= 0 ,0
Exp/Cntr=0.3,0.1

Type RM Length L Ch R = 1 ,54119   ,971,971,971
BEGIN DESCRIPTION:
KEECHIE CREEK 78.0
END DESCRIPTION:
XS GIS Cut Line= 3
      3720017.17     10639715.69       3719792.2     10640918.61
      3719278.63     10642046.62
#Sta/Elev= 30
  4064.6  285.46  4297.1  275.13  4374.4     269  4659.2   264.7    4822   264.1
  4964.4  265.61  4984.8  262.07    4995   262.2  5015.3  265.87  5125.3  263.83
  5208.1  263.62  5573.7  261.92  5576.5  261.42  5579.7  261.92  5685.7  262.76
  5729.6   265.7  5751.6  265.41  5761.2  263.47  5766.7  264.63  5828.5  263.42
  6100.4  267.22  6175.1  272.41  6203.6   277.6  6272.8  283.34  6295.8  286.83
  6355.9  289.77    6388  294.09  6399.9  297.16  6508.8  305.56  6527.8  309.16
#Mann= 5 ,-1 , 0
  4064.6     .12       0  5125.3     .05       0  5208.1     .12       0
  5573.7     .07       0  5579.7     .12       0
Bank Sta=4964.4,5015.3
XS Rating Curve= 0 ,0
Exp/Cntr=0.3,0.1

Type RM Length L Ch R = 1 ,53148   ,496,496,496
BEGIN DESCRIPTION:
KEECHIE CREEK 77.0
END DESCRIPTION:
XS GIS Cut Line= 3
       3719549.6     10639810.21      3719349.61     10640610.19
      3718549.59     10641410.21
#Sta/Elev= 30
  4217.7  306.81    4277  299.75  4331.1  295.75  4382.6  289.96    4447   285.5
  4483.1  281.02  4488.3  281.54  4565.6  274.39  4653.2  268.55  4689.3  264.02
  4694.4   264.8  4722.8  262.86  4771.7  262.08  4895.4  263.45  4900.6  262.06
  4970.1  264.33  5008.4  261.11  5011.1  260.61  5014.4  261.11  5019.1  261.35
  5024.3  263.75  5036.6  264.42  5070.6  262.63  5084.7  264.29  5367.6  262.69
  5848.4  268.27  5919.1   271.7    6004  278.29    6103  287.71  6173.7  297.75
#Mann= 4 ,-1 , 0
  4217.7     .12       0  5008.4     .07       0  5014.4     .12       0
  5036.6     .05       0
Bank Sta=4653.2,5848.4
XS Rating Curve= 0 ,0
Exp/Cntr=0.3,0.1

Type RM Length L Ch R = 1 ,52652   ,1129,1129,1129
BEGIN DESCRIPTION:
KEECHIE CREEK 76.0
END DESCRIPTION:
XS GIS Cut Line= 3
      3719499.59     10639710.21      3719099.61     10640160.19
      3718399.61     10641560.19
#Sta/Elev= 30
  4427.1  314.56  4476.8  309.82  4483.5  307.53  4540.4  301.23  4738.6  287.03
  4809.6  283.34  4908.7  274.18    4951  268.31  4965.2  262.38  4986.9  262.01
  4990.6   260.5  4993.4     260  4996.6   260.5  5007.8  264.03  5087.8  262.44
  5199.6  263.48    5318     262  5425.6  261.01    5519  261.24  5744.7  262.29
  5878.8  264.83  5959.9     268  6222.6  281.58  6289.7   286.4  6348.4  291.55
  6393.1  298.21  6451.8  303.57  6468.6  307.19  6535.7  315.22  6594.4   319.6
#Mann= 7 ,-1 , 0
  4427.1     .12       0  4990.6     .07       0  4996.6     .12       0
    5318     .07       0  5425.6     .05       0    5519     .12       0
  5878.8     .05       0
Bank Sta=4951,5959.9
XS Rating Curve= 0 ,0
Exp/Cntr=0.3,0.1

Type RM Length L Ch R = 1 ,51523   ,549,549,549
BEGIN DESCRIPTION:
KEECHIE CREEK 75.0
END DESCRIPTION:
XS GIS Cut Line= 3
      3719649.63     10639460.18      3718249.61     10640160.19
      3718199.61      10640560.2
#Sta/Elev= 30
  3435.5  326.06  3449.5  325.51  3502.6  318.86    3606  311.56  3622.8     309
  3628.4  309.55  3645.2  306.34  3673.1  304.51  3689.9  301.55  3762.5  296.87
    3852     289  3874.4  286.74  3882.7  284.29  3941.4  281.55  4114.7  269.12
  4634.6  261.07    4970   262.6  4978.4  259.13  4989.4  258.86  4992.1  258.36
  4995.4  258.86  5010.8  259.09  5038.6  262.98  5111.6  263.15  5131.8  261.62
  5192.2  266.45  5212.4  270.65  5259.7  276.56  5343.4  285.28  5403.9  288.13
#Mann= 4 ,-1 , 0
  3435.5     .12       0  4989.4     .07       0  4995.4     .12       0
  5259.7     .05       0
Bank Sta=4970,5038.6
XS Rating Curve= 0 ,0
Exp/Cntr=0.3,0.1

Type RM Length L Ch R = 1 ,50974   ,573,573,573
BEGIN DESCRIPTION:
KEECHIE CREEK 74.0
END DESCRIPTION:
XS GIS Cut Line= 3
      3718399.59     10638910.22      3717999.61     10639710.19
      3717249.58     10640310.21
#Sta/Elev= 30
  4100.1  295.82  4144.8  294.88  4225.8  289.38  4234.2  287.39  4292.9  281.33
  4354.4  271.65  4443.9  262.46  4457.8  263.65  4480.2  261.77  4614.4  260.38
    4824  261.39  4846.4  260.11  4963.7  262.14  4986.1  261.55  5005.1  258.72
  5007.8  258.22  5011.1  258.72  5022.5   261.9  5044.9  260.53  5158.6  261.23
  5385.9  263.44  5493.1  266.32  5528.4  264.42  5592.4  268.92    5642  267.95
  5691.6   269.8    5706  268.96  5755.7  272.41  5902.3  286.77    5955  287.88
#Mann= 4 ,-1 , 0
  4100.1     .12       0  5005.1     .07       0  5011.1     .12       0
  5902.3     .16       0
Bank Sta=4457.8,5493.1
XS Rating Curve= 0 ,0
Exp/Cntr=0.3,0.1

Type RM Length L Ch R = 1 ,50401   ,596,596,596
BEGIN DESCRIPTION:
KEECHIE CREEK 73.0
END DESCRIPTION:
XS GIS Cut Line= 3
      3717799.62     10638860.14      3717699.61     10639310.19
      3716899.63     10639910.18
#Sta/Elev= 30
  4552.5  287.43    4614  283.84  4669.1  277.39  4675.5  275.02  4706.2  271.37
  4736.9  264.75  4767.7  260.98  4839.4  259.68  4972.5  261.83  4991.3  258.77
  4994.1  258.27  4997.3  258.77  5035.4  262.77  5056.2  260.48  5424.2  260.08
  5463.5  262.85  5491.6  263.48  5513.5  259.93  5556.2  260.07  5563.5  262.13
  5570.8  260.27  5604.5  259.76  5727.1  260.18  5763.5   262.4    5800  268.17
  5891.6  277.78  5920.8  283.51  5956.2  284.99  6006.2  289.78  6013.5  291.81
#Mann= 5 ,-1 , 0
  4552.5     .12       0  4991.3     .07       0  4997.3     .12       0
  5424.2     .07       0  5604.5     .12       0
Bank Sta=5035.4,5463.5
XS Rating Curve= 0 ,0
Exp/Cntr=0.3,0.1

Type RM Length L Ch R = 1 ,49805   ,546,546,546
BEGIN DESCRIPTION:
KEECHIE CREEK 72.0
END DESCRIPTION:
XS GIS Cut Line= 3
       3717699.6     10638360.21      3717249.61     10638960.19
      3716499.59     10639760.21
#Sta/Elev= 30
  4226.6  310.46  4354.7   293.4  4476.6  285.72  4490.1  282.61  4498.5  283.01
  4640.1  265.21  4769.3  259.28    4963  261.73  4980.7  258.22  4983.4  257.72
  4986.7  258.22    5012  260.91  5082.8  261.22  5146.3  259.57    5394   259.9
  5415.2  263.02  5422.3  261.54  5457.5  266.95    5500   270.7  5507.3  269.86
  5528.3  273.39  5549.8  273.53    5585  277.74  5592.3  276.27  5599.1  278.26
  5627.4  279.82    5681  279.31  5740.8  282.07  5883.2  293.62  6073.2  313.46
#Mann= 5 ,-1 , 0
  4226.6     .12       0  4980.7     .07       0  4986.7     .12       0
    5681     .16       0  5883.2     .12       0
Bank Sta=4640.1,5457.5
XS Rating Curve= 0 ,0
Exp/Cntr=0.3,0.1

Type RM Length L Ch R = 1 ,49259   ,524,524,524
BEGIN DESCRIPTION:
KEECHIE CREEK 71.0
END DESCRIPTION:
XS GIS Cut Line= 3
      3717449.59      10638260.2      3716849.61     10638610.19
      3716649.61     10639360.18
#Sta/Elev= 30
  4318.7  304.92  4341.8  302.25    4348  302.66  4353.8  300.61  4369.5  299.96
  4453.4  287.36  4480.8  283.59  4492.7  280.64    4529  277.57  4551.5  274.01
  4604.4  268.47  4610.2  266.62  4641.6  263.84  4681.6  257.76  4684.3  257.26
  4687.6  257.76  4968.2  261.27  5023.7  258.35  5030.8     261  5054.7  261.52
  5437.6  259.09  5496.5  260.06  5538.5  262.63  5551.5  263.67  5592.9  268.24
  5644.6  276.04  5651.7  278.07    5686  281.71  5706.7  285.75  5789.5  292.63
#Mann= 6 ,-1 , 0
  4318.7     .12       0  4453.4     .16       0    4529     .12       0
  4681.6     .07       0  4687.6     .12       0  5538.5     .16       0
Bank Sta=4641.6,5551.5
XS Rating Curve= 0 ,0
Exp/Cntr=0.3,0.1

Type RM Length L Ch R = 1 ,48735   ,604,604,604
BEGIN DESCRIPTION:
KEECHIE CREEK 70.0
END DESCRIPTION:
XS GIS Cut Line= 3
      3717399.63     10638210.19      3716849.61     10638110.19
      3715699.62     10639210.18
#Sta/Elev= 30
  4423.3  302.13  4518.2  293.25  4638.6  281.04  4748.6  265.25  4819.7  256.05
  4838.8  258.95  4843.9  255.96  4860.4  258.65  4972.2  258.68  4989.4  255.95
  5003.6  258.57  5010.5  255.72  5017.7   259.7  5123.7  260.86  5166.2  258.38
  5236.9  260.25  5654.3  257.64  5689.5  256.29  5693.7  253.83  5696.5  253.33
  5699.7  253.83  5880.7  263.59  6031.2   270.6  6114.1  269.51    6143  272.88
  6177.6  272.13  6276.7   284.3  6439.3   295.6    6489  303.64  6573.7  311.11
#Mann= 7 ,-1 , 0
  4423.3     .12       0  4518.2     .16       0  4638.6     .12       0
  5693.7     .07       0  5699.7     .12       0  6031.2     .16       0
    6143     .05       0
Bank Sta=4748.6,5880.7
XS Rating Curve= 0 ,0
Exp/Cntr=0.3,0.1

Type RM Length L Ch R = 1 ,48131   ,508,508,508
BEGIN DESCRIPTION:
KEECHIE CREEK 69.0
END DESCRIPTION:
XS GIS Cut Line= 3
       3716699.6     10637360.21      3716449.61     10637910.19
      3715799.61     10638710.19
#Sta/Elev= 30
  4419.2  312.13  4577.4  298.37  4759.7  273.38  4795.9  271.12  4813.5  266.92
  4870.6  260.93  4893.7  257.67  4946.4  256.85  4957.4   252.6  4968.4  256.41
  4979.4  251.86  5001.4  251.88    5009  254.91  5014.5  252.18  5020.6  255.86
  5044.9  256.76  5187.1  257.72  5577.4  256.41  5591.5  255.29  5602.9  251.69
  5605.6  251.19  5608.9  251.69  5620.2  255.81  5655.4  254.55  5698.5  257.52
  5762.5  257.85  5797.6  262.06  5903.4   270.6  5989.7  278.72  6054.1  281.29
#Mann= 4 ,-1 , 0
  4419.2     .12       0  5602.9     .07       0  5608.9     .12       0
  5903.4     .05       0
Bank Sta=4870.6,5797.6
XS Rating Curve= 0 ,0
Exp/Cntr=0.3,0.1

Type RM Length L Ch R = 1 ,47623   ,522,522,522
BEGIN DESCRIPTION:
KEECHIE CREEK 68.0
END DESCRIPTION:
XS GIS Cut Line= 3
      3716699.63     10637260.18      3715999.61     10637760.19
      3715399.58     10638560.23
#Sta/Elev= 30
  4172.9  319.29  4216.2  314.26  4352.3  297.63  4373.2  296.56  4402.7  291.59
  4408.9  292.57  4488.7  282.33  4574.8  274.09  4660.8  268.12  4746.8  268.04
    4812     263    4839  258.43    4898   255.6    4984  255.05  4996.3  249.86
  5001.9  249.69  5004.6  249.19  5007.9  249.69    5011  252.31  5033.2  254.65
  5369.6  254.65  5390.4  250.09  5396.7   250.7    5405  254.75  5419.6  252.43
  5425.9  254.61  5640.4  261.52  5693.8  265.77  5825.9  273.43  6033.2  281.34
#Mann= 5 ,-1 , 0
  4172.9     .05       0  4216.2     .12       0  5001.9     .07       0
  5007.9     .12       0  5693.8     .05       0
Bank Sta=4984,5033.2
XS Rating Curve= 0 ,0
Exp/Cntr=0.3,0.1

Type RM Length L Ch R = 1 ,47101   ,517,517,517
BEGIN DESCRIPTION:
KEECHIE CREEK 67.0
END DESCRIPTION:
XS GIS Cut Line= 3
      3715949.61     10637010.18      3715549.61     10637610.19
      3714749.64     10637960.18
#Sta/Elev= 30
  4279.3   294.9    4374  290.39    4416   286.9  4423.5  285.15    4431  285.69
  4503.2  277.72  4531.7  275.39  4545.2  275.61  4567.8  272.93  4581.3  273.07
    4748  264.09  4820.1  254.11  4878.7  252.71  4986.9  253.93  4992.9  251.47
  4997.4  248.18  5006.4   248.1  5009.1   247.6  5012.4   248.1  5022.2  252.77
  5038.2  254.16  5113.9  255.73  5311.9  264.02  5416.4  265.89  5480.7   268.5
    5492  270.21  5502.5  269.61  5557.5  273.81  5684.4  278.35  5873.6  287.65
#Mann= 5 ,-1 , 0
  4279.3     .12       0  5006.4     .07       0  5012.4     .12       0
  5557.5     .07       0  5684.4     .12       0
Bank Sta=4986.9,5038.2
XS Rating Curve= 0 ,0
Exp/Cntr=0.3,0.1

Type RM Length L Ch R = 1 ,46584   ,512,512,512
BEGIN DESCRIPTION:
KEECHIE CREEK 66.0
END DESCRIPTION:
XS GIS Cut Line= 3
      3715849.64     10637010.18      3715399.61     10637210.19
       3714599.6      10637910.2
#Sta/Elev= 30
  4506.4  290.58  4604.9  282.16  4637.1  276.87  4642.5  278.23  4665.8  273.01
  4671.3  273.98  4681.5   272.8    4689  269.74  4694.5  271.05  4816.3  259.22
  4823.8  257.39    4977  253.61  4984.5  252.43  4993.1  248.58  4995.9  248.08
  4999.1  248.58  5012.6  251.47  5140.8  252.79  5190.1  251.51  5317.8  257.61
  5459.7  259.43  5551.7  262.41    5585  264.91  5615.3   268.4  5735.9  272.45
  5764.3  271.99  5818.7  276.53  5849.3  279.74  5899.1  281.36  6061.9  292.89
#Mann= 5 ,-1 , 0
  4506.4     .12       0  4993.1     .07       0  4999.1     .12       0
    5585     .07       0  5818.7     .12       0
Bank Sta=4977,5012.6
XS Rating Curve= 0 ,0
Exp/Cntr=0.3,0.1

Type RM Length L Ch R = 1 ,46072   ,553,553,553
BEGIN DESCRIPTION:
KEECHIE CREEK 65.0
END DESCRIPTION:
XS GIS Cut Line= 3
      3715749.61     10636160.18      3714949.61     10636960.19
      3714149.64     10637760.15
#Sta/Elev= 30
  3893.2  295.64  3935.6  292.48  3992.2  285.65  4020.5  284.27  4062.9  278.78
  4133.6  271.93  4190.2  268.15  4232.6  262.78  4260.9  261.23  4430.6  261.86
    4473  259.78  4883.2  253.51  4897.3  251.83  4911.4  252.99  4925.6  251.81
    4968  252.06  4993.3  247.23    4996  246.73  4999.3  247.23  5010.4  250.36
    5021  251.29  5038.7  250.44  5321.6   251.8    5463  250.63  5632.7  251.66
  5788.3   267.9  5943.8  279.42  5959.2  281.49  6152.4  303.59  6155.9  303.59
#Mann= 5 ,-1 , 0
  3893.2     .12       0  4993.3     .07       0  4999.3     .12       0
  5959.2     .16       0  6152.4     .12       0
Bank Sta=4968,5021
XS Rating Curve= 0 ,0
Exp/Cntr=0.3,0.1

Type RM Length L Ch R = 1 ,45519   ,572,572,572
BEGIN DESCRIPTION:
KEECHIE CREEK 64.0
END DESCRIPTION:
XS GIS Cut Line= 3
      3714399.61     10636060.17      3714449.61     10636810.19
       3713849.6      10637610.2
#Sta/Elev= 30
  4224.8   299.7  4274.9  296.07  4335.1  289.75  4345.1  287.27  4415.2  278.97
  4445.3  272.38  4485.4  266.53  4575.6  260.19  4635.7  253.95    4756  250.46
  4926.4  251.38  4956.4   250.5  4979.6  251.47  4983.8  247.31  4995.4  246.81
  4998.1  246.31  5001.4  246.81  5012.9  251.26  5069.2  251.38  5126.5   249.5
  5554.6  251.13  5626.5  257.85  5654.6  262.01    5690   265.1  5698.4  267.06
  5819.2  278.35  5826.5  280.58  5854.6  283.52  5883.8  288.79  5976.5   300.8
#Mann= 3 ,-1 , 0
  4224.8     .12       0  4995.4     .07       0  5001.4     .12       0
Bank Sta=4979.6,5012.9
XS Rating Curve= 0 ,0
Exp/Cntr=0.3,0.1

Type RM Length L Ch R = 1 ,44947   ,533,533,533
BEGIN DESCRIPTION:
KEECHIE CREEK 63.0
END DESCRIPTION:
XS GIS Cut Line= 3
       3714299.6      10636060.2      3714049.61     10636410.19
       3713399.6      10637210.2
#Sta/Elev= 30
    4542   294.9  4549.4  295.55  4555.5  293.39  4570.3  291.91  4578.9  292.73
    4714  283.22  4736.2  277.91  4742.3  279.24  4792.7  268.54  4849.2  261.15
  4908.2  256.35  4914.3   254.5  4975.3  250.83  4997.1  247.88  4999.9  247.38
  5003.1  247.88  5014.5  250.36  5199.8  249.09  5292.5  251.08  5484.3  248.74
  5583.4  251.91  5597.8  254.49  5647.3     254  5696.9  255.86    5740  259.61
  5818.3  263.62  5839.1  263.23  5875.5  266.52  5952.6  275.08  6002.9  282.91
#Mann= 4 ,-1 , 0
    4542     .12       0  4997.1     .07       0  5003.1     .12       0
  5875.5     .16       0
Bank Sta=4914.3,5597.8
XS Rating Curve= 0 ,0
Exp/Cntr=0.3,0.1

Type RM Length L Ch R = 1 ,44414   ,531,531,531
BEGIN DESCRIPTION:
KEECHIE CREEK 62.0
END DESCRIPTION:
XS GIS Cut Line= 3
      3714349.65     10635960.17      3713549.61     10636260.19
      3712749.62     10637060.18
#Sta/Elev= 30
  4133.7  303.73  4148.9  302.77  4155.1  300.78  4251.2  286.82  4344.7   276.6
  4368.7   275.2  4399.9  270.63  4405.2  271.31  4545.8  256.56  4631.3  249.76
  4755.7  249.35  4801.2  249.35  4827.1  249.35  4832.4  253.15  4857.3  253.23
  4881.3   250.4    4973  250.14  4978.4  246.99  4982.5  246.74  4985.2  246.24
  4988.5  246.74  5044.7  249.28  5143.7  247.78  5454.8  248.58    5568  252.56
  5593.1  253.15    5766  260.07    5865  268.65  6006.4  284.18  6119.5  289.57
#Mann= 6 ,-1 , 0
  4133.7     .12       0  4755.7     .07       0  4801.2     .12       0
  4982.5     .07       0  4988.5     .12       0  5593.1     .05       0
Bank Sta=4857.3,5568
XS Rating Curve= 0 ,0
Exp/Cntr=0.3,0.1

Type RM Length L Ch R = 1 ,43883   ,538,538,538
BEGIN DESCRIPTION:
KEECHIE CREEK 61.0
END DESCRIPTION:
XS GIS Cut Line= 3
      3713999.64     10635210.16      3713249.61     10635860.19
      3712499.61     10636660.19
#Sta/Elev= 30
  4007.8  312.49  4050.1  310.68  4057.7  312.32    4072   308.4  4156.5  298.48
  4192.6  296.15  4199.2  294.24  4348.3   283.8  4369.2  280.85  4432.8  277.68
  4532.6   266.7  4567.7  260.83  4659.8  252.79  4725.7  249.35  4817.9   248.4
  4993.2  249.26    4997  247.01  5004.4  246.77  5007.1  246.27  5010.4  246.77
  5035.7  248.88  5120.7  247.38  5290.2  248.18  5400.8  253.35  5481.2  252.36
  5594.5  255.27  5665.3  254.82  5757.2  261.05  5898.8  267.11  6096.9  282.99
#Mann= 6 ,-1 , 0
  4007.8     .12       0  4725.7     .05       0  4817.9     .12       0
  5004.4     .07       0  5010.4     .12       0  5400.8     .05       0
Bank Sta=4659.8,5400.8
XS Rating Curve= 0 ,0
Exp/Cntr=0.3,0.1

Type RM Length L Ch R = 1 ,43345   ,377,377,377
BEGIN DESCRIPTION:
KEECHIE CREEK 60.0
END DESCRIPTION:
XS GIS Cut Line= 3
      3713899.58      10635210.2      3713099.61     10635410.19
      3712399.63     10636660.15
#Sta/Elev= 30
  4200.1  301.09  4300.6  289.77  4305.7  290.24  4424.3  278.03  4429.4   278.6
    4548  265.97  4635.6  260.12  4671.6  256.44    4718  255.62  4795.3  249.08
  4940.8  247.71  4993.8  247.39  5003.6  244.97  5006.4  244.47  5009.6  244.97
  5014.4  247.41  5069.6  247.43    5231   249.3  5421.9  249.19  5494.6  252.07
  5562.3  250.88  5686.8   251.6  5746.1  254.44  5773.6  257.74  5832.9  261.09
  6178.8  265.99  6238.1  270.11    6309   277.9  6368.3  282.19  6457.3  286.07
#Mann= 5 ,-1 , 0
  4200.1     .12       0  4940.8     .07       0  5003.6     .07       0
  5009.6     .07       0  5069.6     .05       0
Bank Sta=4993.8,5014.4
XS Rating Curve= 0 ,0
Exp/Cntr=0.3,0.1

Type RM Length L Ch R = 1 ,42968   ,756,756,756
BEGIN DESCRIPTION:
KEECHIE CREEK 59.0
END DESCRIPTION:
XS GIS Cut Line= 4
      3713129.55      10634173.3       3713016.7     10634919.86
       3712660.8     10635440.69      3712296.21     10636673.35
#Sta/Elev= 30
  3998.3  302.08    4157  284.62  4168.7  284.88  4217.7  279.62  4301.3  274.34
  4349.1   269.1  4379.5  268.29  4521.1  258.78  4648.9   254.9  4701.2  253.77
  4733.4  254.83  4743.6  252.59  4809.2  249.95  4982.6  247.96  4985.7  245.14
  4988.4  244.64  4991.7  245.14  5003.6  247.96  5024.6  248.93  5157.9  249.25
  5356.5  250.42  5474.4  254.12  5529.6  257.69  5592.2  259.49  5971.5  261.57
  6280.5  265.81  6353.1  269.77  6424.8  276.74  6496.6  281.04  6669.6  285.95
#Mann= 6 ,-1 , 0
  3998.3     .12       0  4648.9     .16       0  4701.2     .12       0
  4985.7     .07       0  4991.7     .12       0  5157.9     .05       0
Bank Sta=4733.4,5474.4
XS Rating Curve= 0 ,0
Exp/Cntr=0.3,0.1

Type RM Length L Ch R = 1 ,42212   ,473,473,473
BEGIN DESCRIPTION:
KEECHIE CREEK 58.0
END DESCRIPTION:
XS GIS Cut Line= 3
      3712704.19     10634372.99      3711948.99     10634963.26
      3710882.95     10635041.26
#Sta/Elev= 30
  4529.3  310.76  4553.4  311.44  4576.4  310.74  4694.5  304.88  4887.1  283.59
  4922.4  277.96  4943.2   264.4  4979.3  250.13  4998.1  243.07  5000.8  242.57
  5004.1  243.07  5015.5  248.22  5036.4  249.95  5100.8  248.12    5547  259.27
  5637.6  264.17  5651.9  266.33  5657.6  270.12  5722.8  278.99  5858.2  294.41
  6138.9  290.58    6169  281.16  6196.7  283.14  6219.1  278.93  6249.2  283.63
  6299.7  283.72  6339.1  283.18  6399.6  282.92  6419.7  285.45  6556.7  282.88
#Mann= 10 ,-1 , 0
  4529.3     .12       0  4553.4     .16       0  4576.4     .12       0
  4998.1     .07       0  5004.1     .12       0  5100.8     .05       0
    5547     .16       0  5722.8     .05       0  6299.7     .12       0
  6339.1     .16       0
Bank Sta=4979.3,5036.4
XS Rating Curve= 0 ,0
Exp/Cntr=0.3,0.1

Type RM Length L Ch R = 1 ,41739   ,454,454,454
BEGIN DESCRIPTION:
KEECHIE CREEK 57.0
END DESCRIPTION:
XS GIS Cut Line= 3
      3712499.64     10634310.19      3712099.61     10634260.19
      3711699.62     10634810.18
#Sta/Elev= 30
  4591.5  303.46  4601.6  303.43  4662.1  294.18  4752.8  283.27  4833.4  270.31
  4863.6  267.08  4871.2  264.53  4944.3   257.5  4951.8  255.39  4956.8  255.63
  4984.6  250.84  4992.1   245.5  4997.7   245.5    5002  243.02  5013.7   242.9
  5016.4   242.4  5019.7   242.9  5037.5   248.1  5044.1  247.06  5058.4  248.61
  5073.1  248.48  5087.8  246.85  5113.8  248.19  5259.3  249.47  5324.2  251.28
  5439.4  257.02  5533.4  266.39    5546  266.49  5596.3  278.19  5674.7  287.79
#Mann= 5 ,-1 , 0
  4591.5     .12       0  5013.7     .07       0  5019.7     .12       0
  5113.8     .05       0  5533.4     .16       0
Bank Sta=4984.6,5037.5
XS Rating Curve= 0 ,0
Exp/Cntr=0.3,0.1

Type RM Length L Ch R = 1 ,41285   ,657,657,657
BEGIN DESCRIPTION:
KEECHIE CREEK 56.0
END DESCRIPTION:
XS GIS Cut Line= 3
      3712530.54     10634155.96      3711384.76     10633826.11
      3710144.03     10634034.34
#Sta/Elev= 30
  4288.8  287.88  4544.7  267.98  4549.9  265.52  4664.4  253.66  4728.7  249.26
  4974.9  248.41  4980.1  248.37    4987  242.83  4994.4  242.77  4997.1  242.27
  5000.4  242.77  5028.6  248.93  5088.1  248.02  5408.2  255.14  5491.2   256.5
  5668.9  264.05  5837.3  277.04  5891.9  281.61  5902.8  285.27  5963.4  288.39
  6145.4  290.55  6216.4  289.73  6256.4   281.8  6261.5  283.16  6267.1  278.86
  6377.7  294.92  6382.8  293.12  6440.6  298.67  6540.9  307.03  6739.2  313.69
#Mann= 8 ,-1 , 0
  4288.8     .12       0  4994.4     .07       0  5000.4     .12       0
  5088.1     .05       0  5408.2     .16       0  5491.2     .05       0
  5837.3     .16       0  6440.6     .05       0
Bank Sta=4974.9,5028.6
XS Rating Curve= 0 ,0
Exp/Cntr=0.3,0.1

Type RM Length L Ch R = 1 ,40628   ,1018,1018,1018
BEGIN DESCRIPTION:
KEECHIE CREEK 55.0
END DESCRIPTION:
XS GIS Cut Line= 3
      3712649.58     10634210.15      3711899.61     10633410.19
      3711099.62      10632610.2
#Sta/Elev= 30
  3875.6  299.28  3900.7  296.02  4040.8  280.38  4179.6  267.75  4278.8  260.38
  4457.5  250.99  4459.2  250.96  4558.5  248.03  4625.6  247.66  4674.9  249.65
  4696.4  248.11  4795.1  248.68  4816.6  247.18  4837.6  249.25    4944  248.54
  4965.1  247.49  4997.4  241.98  5000.2  241.48  5003.4  241.98    5018  243.34
  5028.7   247.3    5057  248.38  5146.7  247.79  5255.8  247.78  5382.3  248.04
  5580.3  255.68  5721.7  266.45  5933.8  287.82  6046.9  297.05  6103.5  299.55
#Mann= 12 ,-1 , 0
  3875.6     .12       0  3900.7     .16       0  4040.8     .12       0
  4179.6     .16       0  4457.5     .12       0  4459.2     .16       0
  4558.5     .12       0  4997.4     .07       0  5003.4     .12       0
    5018     .07       0  5146.7     .05       0  5255.8     .12       0
Bank Sta=4944,5057
XS Rating Curve= 0 ,0
Exp/Cntr=0.3,0.1

Type RM Length L Ch R = 1 ,39610   ,588,588,588
BEGIN DESCRIPTION:
KEECHIE CREEK 54.0
END DESCRIPTION:
XS GIS Cut Line= 3
      3712849.62     10632010.18      3712049.61     10632660.19
      3711249.62     10632460.19
#Sta/Elev= 30
  3973.1  292.68  3994.7  292.58  4029.9  284.43  4188.9  270.68  4378.3  255.31
  4427.8  250.55  4577.9  246.88  4939.5   246.7  4953.6  245.22  4956.3  242.54
  4958.5  240.35  4961.3  239.85  4964.5  240.35    4968  246.77  4975.9  243.23
  4982.3   245.1  4990.3  241.48  4996.7   244.9  5000.7  241.32  5006.5  241.32
  5045.1  247.34  5086.3  245.94  5104.4  242.22  5168.8  247.62  5274.5  248.72
  5467.2  264.78  5533.3  265.35  5653.3  273.66  5805.3  292.26  5828.5  292.96
#Mann= 8 ,-1 , 0
  3973.1     .12       0  4188.9     .16       0  4378.3     .05       0
  4956.3     .12       0  4958.5     .07       0  4964.5     .12       0
  5467.2     .05       0  5533.3     .12       0
Bank Sta=4939.5,5168.8
XS Rating Curve= 0 ,0
Exp/Cntr=0.3,0.1

Type RM Length L Ch R = 1 ,39022   ,550,550,550
BEGIN DESCRIPTION:
KEECHIE CREEK 53.0
END DESCRIPTION:
XS GIS Cut Line= 3
      3712649.64     10632010.18      3711849.61     10632210.19
      3711199.63     10632410.18
#Sta/Elev= 30
  4182.1  271.67  4206.2  269.72  4287.8  262.75  4377.4  252.76  4411.5  252.29
  4419.2  250.74  4571.2  250.74  4594.4  254.64  4604.7  253.83  4617.6  250.09
  4625.4  246.04  4635.7  245.21  4736.2  243.93  4955.2  245.44  4979.9  242.32
  4985.7  240.22  4988.5  239.72  4991.7  240.22  5017.2  242.48  5028.3  246.06
  5055.8  244.85  5132.3  246.21  5224.5  245.38  5236.9  247.98  5333.1  256.86
  5431.1  263.24    5509  273.35  5540.3  280.24  5599.9  289.31  5686.8  298.54
#Mann= 6 ,-1 , 0
  4182.1     .12       0  4206.2     .16       0  4377.4     .05       0
  4979.9     .12       0  4985.7     .07       0  4991.7     .12       0
Bank Sta=4955.2,5028.3
XS Rating Curve= 0 ,0
Exp/Cntr=0.3,0.1

Type RM Length L Ch R = 1 ,38472   ,371,371,371
BEGIN DESCRIPTION:
KEECHIE CREEK 52.0
END DESCRIPTION:
XS GIS Cut Line= 3
      3712572.04     10631147.67      3711408.87     10631974.04
       3711040.8      10632293.5
#Sta/Elev= 30
  3588.3  292.75  3641.1   285.8  3649.8  286.38  3655.9  283.83  3691.6  278.21
  3700.2  278.54  3721.1  273.65  3828.1  263.93  3914.2  252.36  4044.6  248.59
  4166.4  247.41  4206.5  248.63  4310.2  246.32  4359.5  244.14  4550.8  243.13
  4910.4  244.33  4976.9  244.69  4994.8  239.04  4997.6  238.54  5000.8  239.04
  5018.8  240.22  5026.5   245.4  5061.6  243.22  5110.9  246.59    5317  272.72
  5366.4  280.97  5394.9  288.93  5415.8  292.31  5465.1  298.67  5502.5  301.04
#Mann= 7 ,-1 , 0
  3588.3     .12       0  4206.5     .05       0  4310.2     .12       0
  4550.8     .05       0  4910.4     .12       0  4994.8     .07       0
  5000.8     .12       0
Bank Sta=4976.9,5026.5
XS Rating Curve= 0 ,0
Exp/Cntr=0.3,0.1

Type RM Length L Ch R = 1 ,38101   ,115,115,115
BEGIN DESCRIPTION:
Mapping XS d688e083
END DESCRIPTION:
XS GIS Cut Line= 2
      3711888.07     10631092.07      3710759.57     10632119.87
#Sta/Elev= 30
    4117   283.3  4121.7  281.75  4135.8  284.23  4155.1  281.94  4284.5  276.97
  4404.8  254.83  4440.6  250.75  4447.3  250.53  4518.3  242.61  4738.8  242.63
  4944.6  243.17    4971  244.35  4978.4  242.87  4982.2  239.58  4984.9  239.08
  4988.2  239.58  5006.8  241.05  5013.5  243.55  5056.1  240.78  5070.3  243.33
  5155.4  244.25  5225.7  249.58  5318.3  257.62  5445.3  275.31  5452.7  274.55
  5473.7  278.43  5487.9  278.07  5516.2  281.64  5585.1  295.22  5643.4  298.26
#Mann= 8 ,-1 , 0
    4117      .1       0  4155.1     .16       0  4440.6     .12       0
  4738.8     .05       0  4944.6     .12       0  4982.2     .07       0
  4988.2     .12       0  5585.1     .05       0
Bank Sta=4447.3,5225.7
XS Rating Curve= 0 ,0
Exp/Cntr=0.3,0.1

Type RM Length L Ch R = 1 ,37986   ,157,157,157
BEGIN DESCRIPTION:
KEECHIE CREEK 51.0
END DESCRIPTION:
XS GIS Cut Line= 2
      3711804.69     10631043.49      3710683.87     10632063.69
#Sta/Elev= 30
  4088.9  283.83  4110.6  284.21  4238.9  277.03  4253.1  273.33  4281.4  270.06
  4330.8  258.26  4369.1  253.49  4436.8  247.93    4451  244.83  4477.3  244.29
    4515  244.46    4562  241.82    4617  241.89  4700.7  242.92  4833.5  241.98
  4896.5  243.55    4978  242.83  4993.3  240.02  4996.1  239.52  4999.3  240.02
  5010.5  240.81  5024.7  247.61  5036.3  247.56  5059.8  243.67  5197.6  252.55
  5375.4  268.96  5470.7  276.94  5532.6  285.31  5595.3  288.94  5604.5  289.23
#Mann= 16 ,-1 , 0
  4088.9     .05       0  4110.6     .16       0  4369.1     .05       0
  4477.3     .12       0    4562     .08       0    4617     .12       0
  4700.7     .05       0  4896.5     .12       0    4978     .08       0
  4993.3     .07       0  4999.3     .08       0  5036.3     .12       0
  5197.6     .05       0  5375.4     .12       0  5532.6     .08       0
  5595.3     .05       0
Bank Sta=4436.8,5024.7
XS Rating Curve= 0 ,0
Exp/Cntr=0.3,0.1

Type RM Length L Ch R = 1 ,37829   ,130,130,130
BEGIN DESCRIPTION:
Mapping XS f7b31e06
END DESCRIPTION:
XS GIS Cut Line= 2
      3711763.03     10630876.82      3710540.78     10631984.49
#Sta/Elev= 30
    4032  272.55  4058.1  270.61  4064.9  266.31  4086.5  267.26  4114.9  261.76
  4126.6  262.52  4164.2  265.46  4178.4   263.1  4265.2  263.19  4355.5  253.34
    4490  244.44  4600.9  241.66  4630.2  240.51    4797  242.98  4851.9  242.84
  4937.1   243.8  4985.3  244.38  4990.3  241.66    5004     238  5006.7   237.5
    5010     238  5027.9  238.34  5035.3  243.66  5141.5  243.93  5351.2  269.57
  5438.8  285.77  5509.1  287.44  5543.7  292.87  5637.4  298.47  5681.5  299.55
#Mann= 14 ,-1 , 0
    4032     .12       0  4126.6     .05       0  4265.2     .12       0
  4600.9     .08       0  4630.2     .12       0    4797     .05       0
  4851.9     .12       0  4937.1     .08       0  4990.3     .12       0
    5004     .07       0    5010     .12       0  5351.2     .05       0
  5543.7     .16       0  5637.4     .05       0
Bank Sta=4985.3,5035.3
XS Rating Curve= 0 ,0
Exp/Cntr=0.3,0.1

Type RM Length L Ch R = 1 ,37699   ,277,277,277
BEGIN DESCRIPTION:
Mapping XS ae3d074a
END DESCRIPTION:
XS GIS Cut Line= 2
       3711665.8      10630817.8      3710479.22     10631876.01
#Sta/Elev= 30
  4115.2   281.4  4121.6  281.97  4128.3  279.76    4150  278.37  4156.7  275.99
  4170.9  275.51  4248.6   264.3  4326.4   256.2  4333.9  253.71  4376.6  254.68
  4475.2  249.81    4553   243.4  4659.5  241.93  4687.6  240.06  4709.3  241.57
  4900.6  241.77  4985.2  244.68  5003.9  237.92  5006.7  237.42  5009.9  237.92
  5027.9  243.26  5098.9   241.9  5211.8  247.98  5268.6  253.46  5346.4  263.69
  5474.3  284.33  5495.2  289.49  5626.7  299.82  5672.2  300.86  5705.1  301.95
#Mann= 5 ,-1 , 0
  4115.2     .12       0  5003.9     .07       0  5009.9     .12       0
  5626.7     .16       0  5672.2     .05       0
Bank Sta=4985.2,5027.9
XS Rating Curve= 0 ,0
Exp/Cntr=0.3,0.1

Type RM Length L Ch R = 1 ,37422   ,587,587,587
BEGIN DESCRIPTION:
KEECHIE CREEK 50.0
END DESCRIPTION:
XS GIS Cut Line= 3
      3711649.61     10630660.19      3710849.61     10631210.19
      3710499.61     10631560.19
#Sta/Elev= 30
  4042.7  293.23  4208.5  281.45  4251.8  275.75  4309.3  267.97  4351.9  261.23
  4406.4  255.36  4487.6  245.11  4661.6  241.95    4698  240.63  4710.4  238.67
  4734.1  241.18  4776.1  242.61  4811.9  242.69  4826.8  240.08  4847.8  239.67
  4862.7  242.68  4970.2  243.11  4985.1  238.17  4991.2  239.37    4997  238.17
  4999.8  237.67    5003  238.17  5027.7   243.6  5070.1  242.65  5183.2  246.87
  5253.9     252  5326.8   259.9  5359.3  263.98  5409.5  271.12  5508.5  290.87
#Mann= 9 ,-1 , 0
  4042.7     .12       0  4251.8     .16       0  4309.3     .12       0
  4406.4     .16       0  4487.6     .12       0    4997     .07       0
    5003     .12       0  5326.8     .16       0  5359.3     .12       0
Bank Sta=4970.2,5027.7
XS Rating Curve= 0 ,0
Exp/Cntr=0.3,0.1

Type RM Length L Ch R = 1 ,36835   ,771,771,771
BEGIN DESCRIPTION:
KEECHIE CREEK 49.0
END DESCRIPTION:
XS GIS Cut Line= 3
      3711249.63     10630360.17      3710799.61     10630710.19
      3709999.63     10631060.18
#Sta/Elev= 30
  4409.2  300.03  4478.3  292.15    4487  290.04  4509.7   289.7  4530.5  287.28
  4665.3  270.34  4673.5  270.99  4814.6   250.4  4865.3   243.3  4901.5  241.39
  4925.6  236.78  4928.4  236.28  4931.6  236.78  4941.6  240.42  4993.7  242.27
  5001.1  237.68  5017.1  237.17    5023  240.73  5033.9  242.67  5121.6  240.16
  5379.8  247.67  5432.1  249.35  5448.7   249.9  5541.1  252.49  5645.5  259.72
  5677.9  263.03  5699.7  267.34  5727.4  275.43  5754.3  280.41  5852.5  286.51
#Mann= 8 ,-1 , 0
  4409.2     .05       0  4478.3     .16       0  4925.6     .07       0
  4931.6     .16       0  4941.6     .12       0  5379.8     .05       0
  5432.1     .16       0  5727.4     .12       0
Bank Sta=4814.6,5448.7
XS Rating Curve= 0 ,0
Exp/Cntr=0.3,0.1
