--- MACK CREEK.prj (project) ---

Proj Title=MACK CREEK Base Level Engineering
Current Plan=p01
Default Exp/Contr=0.3,0.1
English Units
Geom File=g01
Flow File=f01
Plan File=p01
Y Axis Title=Elevation
X Axis Title(PF)=Main Channel Distance
X Axis Title(XS)=Station
BEGIN DESCRIPTION:
MACK CREEK
END DESCRIPTION:
DSS Export Rating Curves= 0
DSS Export Rating Curve Sorted= 0
DSS Export Volume Flow Curves= 0
DXF OffsetX= 0
DXF OffsetY= 0
DXF ScaleX= 1
DXF ScaleY= 10

--- MACK CREEK.p01 (plan) ---

Plan Title=Multiple Run
Short Identifier=Multiple
Geom File=g01
Flow File=f01
Subcritical Flow
K Sum by GR= 0
Std Step Tol= 0.01
Critical Tol= 0.01
Num of Std Step Trials= 20
Max Error Tol= 0.3
Flow Tol Ratio= 0.001
Split Flow NTrial= 30
Split Flow Tol= 0.02
Split Flow Ratio= 0.02
Log Output Level= 0
Friction Slope Method= 1
Unsteady Friction Slope Method= 2
Unsteady Bridges Friction Slope Method= 1
Parabolic Critical Depth
Global Vel Dist=  1 , 1 , 1
Global Log Level= 0
CheckData=True
Encroach Param= -1, 0, 0, 0
BEGIN DESCRIPTION:
Multiple Run
END DESCRIPTION:

--- MACK CREEK.f01 (steady flow) ---

Flow Title=Multiple
Program Version=4.10
Number of Profiles= 7
Profile Names=10-year,25-year,50-year,1pct_min,100-year,1pct_plu,500-year
River Rch & RM=MACK CREEK,Reach-1         ,30996
     877    1215    1499    1359    1838    2486    2774
River Rch & RM=MACK CREEK,Reach-1         ,28919
    1088    1520    1887    1719    2324    3144    3542
River Rch & RM=MACK CREEK,Reach-1         ,23050
    1270    1787    2228    2038    2756    3728    4235
River Rch & RM=MACK CREEK,Reach-1         ,20933
    1931    2754    3465    3192    4317    5839    6732
River Rch & RM=MACK CREEK,Reach-1         ,20420
    1931    2754    3465    3192    4317    5839    6732
River Rch & RM=MACK CREEK,Reach-1         ,5742
    2029    2900    3655    3371    4559    6166    7128
Boundary for River Rch & Prof#=MACK CREEK,Reach-1         , 1
Up Type= 0
Dn Type= 3
Dn Slope=0.007
Boundary for River Rch & Prof#=MACK CREEK,Reach-1         , 2
Up Type= 0
Dn Type= 3
Dn Slope=0.007
Boundary for River Rch & Prof#=MACK CREEK,Reach-1         , 3
Up Type= 0
Dn Type= 3
Dn Slope=0.007
Boundary for River Rch & Prof#=MACK CREEK,Reach-1         , 4
Up Type= 0
Dn Type= 3
Dn Slope=0.007
Boundary for River Rch & Prof#=MACK CREEK,Reach-1         , 5
Up Type= 0
Dn Type= 3
Dn Slope=0.007
Boundary for River Rch & Prof#=MACK CREEK,Reach-1         , 6
Up Type= 0
Dn Type= 3
Dn Slope=0.007
Boundary for River Rch & Prof#=MACK CREEK,Reach-1         , 7
Up Type= 0
Dn Type= 3
Dn Slope=0.007
DSS Import GetInterval= 0
DSS Import GetPeak= 0
DSS Import FillOption= 0

--- MACK CREEK.g01 (geometry) ---

Geom Title=Existing Conditions
Program Version=4.10

River Reach=MACK CREEK      ,Reach-1
Reach XY= 30
      3738972.36     10609389.15        3738502.       10608464.
        3738389.       10608759.        3737349.     10608153.17
        3736183.     10608411.17      3734067.34       10605369.
        3733392.       10605282.       3733232.5       10604635.
        3731821.       10604477.        3731774.       10604104.
        3730197.       10603128.      3729899.25       10602398.
      3730235.25       10601834.        3729945.       10601610.
      3729583.25       10601853.      3728547.25       10600907.
      3728654.25       10600168.       3727324.5       10599223.
       3726796.5       10597557.        3725752.       10597613.
        3724844.       10596823.      3724870.25       10596482.
      3725277.75       10596757.        3725478.       10596156.
      3725784.75       10596254.      3725840.75       10595693.
      3726255.75       10595957.      3726505.25       10595410.
        3726027.       10595290.      3726252.17     10594860.28

Type RM Length L Ch R = 1 ,30996   ,117,117,117
BEGIN DESCRIPTION:
MACK CREEK 62.0
END DESCRIPTION:
XS GIS Cut Line= 3
      3738999.59      10609160.2      3738899.61     10609210.19
       3738699.6      10609310.2
#Sta/Elev= 30
  4884.6   328.9    4893  328.42  4898.5  327.29  4915.3  325.87  4920.9  323.58
  4929.3  322.19  4937.7  322.59  4951.7  320.68    4960   320.5    4974  318.74
    4988  318.18  4993.6  315.99  4999.2  315.99  5007.4  314.84  5010.1  314.34
  5013.4  314.84  5018.7  318.08  5032.7  318.76  5055.1   318.9  5085.8  320.18
  5094.2  321.14  5108.2  321.17  5122.2  322.49  5130.5  322.68  5144.5  324.46
  5166.9  325.42  5183.6  327.69  5189.2  327.65  5211.6  330.33    5220  330.53
#Mann= 3 ,-1 , 0
  4884.6     .16       0  5007.4     .07       0  5013.4     .16       0
Bank Sta=4988,5018.7
XS Rating Curve= 0 ,0
Exp/Cntr=0.3,0.1

Type RM Length L Ch R = 1 ,30879   ,344,344,344
BEGIN DESCRIPTION:
Mapping XS 0a057f5d
END DESCRIPTION:
XS GIS Cut Line= 5
3739705.5684443210608390.1453157      3739681.48     10608726.05
       3739072.8     10609037.95      3738781.13     10609128.23
      3738545.01     10609171.63
#Sta/Elev= 30
  3752.9  337.44  3933.4  333.58  3973.5  330.07  4083.8  333.09  4147.9  330.36
  4204.1  324.53  4264.6   325.4  4392.2  322.07    4420  324.58  4458.8  322.32
    4481  323.24  4508.8  326.86  4575.4  330.81  4636.4  330.92  4675.1  327.89
  4725.2  330.36  4754.7  328.67  4833.2  329.97  4898.4  326.82  4954.9  318.49
  4975.8  318.06  4998.5  313.18  5001.3  312.68  5004.5  313.18  5017.7  318.26
  5034.1  316.97  5049.1  319.08  5116.7  320.37  5202.5  331.35    5319  337.17
#Mann= 3 ,-1 , 0
  3752.9     .16       0  4998.5     .07       0  5004.5     .16       0
Bank Sta=4975.8,5017.7
XS Rating Curve= 0 ,0
Exp/Cntr=0.3,0.1

Type RM Length L Ch R = 1 ,30535   ,100,100,100
BEGIN DESCRIPTION:
MACK CREEK 61.0
END DESCRIPTION:
XS GIS Cut Line= 5
      3739509.24      10608490.4      3739507.65     10608628.61
      3739331.95     10608713.39      3738927.37     10608926.96
      3738493.31      10608976.1
#Sta/Elev= 30
  3977.4   336.9  4143.3  336.61  4299.5  334.09  4351.1  330.48  4417.1  321.97
  4471.9  322.66  4477.5  319.43  4493.9  320.52  4515.9   316.7  4537.9  319.58
  4543.6  316.62    4582  318.63  4631.7  315.65  4670.1   317.7  4708.4  315.66
  4776.3  315.43  4816.6  319.12  4826.6  317.85  4831.6  318.99  4836.7  316.64
    4887  318.37  4977.6  316.46  4994.7  311.64  4997.5  311.14  5000.7  311.64
  5006.1  317.57  5011.1  316.45  5027.9  327.69  5058.1  331.36  5195.3  334.26
#Mann= 3 ,-1 , 0
  3977.4     .16       0  4994.7     .07       0  5000.7     .16       0
Bank Sta=4977.6,5006.1
XS Rating Curve= 0 ,0
Exp/Cntr=0.3,0.1

Type RM Length L Ch R = 1 ,30435   ,179,179,179
BEGIN DESCRIPTION:
Mapping XS 3e3df57b
END DESCRIPTION:
XS GIS Cut Line= 4
3739218.1083952510608597.6506703      3738998.78     10608754.39
      3738834.95     10608841.77      3738604.33     10608914.59
#Sta/Elev= 30
  4445.1  336.07    4517  333.31  4560.6  334.82  4590.1  334.04    4603  331.55
    4611  332.68  4617.2  331.15  4646.7  332.36  4689.1  331.07    4697  329.11
  4725.1  328.25  4805.7  320.77    4822  317.95  4860.3  315.92  4887.9  311.77
  4937.4  316.46  4940.8  309.92  4943.5  309.42  4946.8  309.92    4949   314.2
  4976.1     310  4989.8  313.29  5000.3   311.3  5021.3  310.56  5040.8  316.74
    5046  314.65  5052.8  322.72  5063.3  325.08  5115.9  329.43  5142.2  329.49
#Mann= 3 ,-1 , 0
  4445.1     .16       0  4940.8     .07       0  4946.8     .16       0
Bank Sta=4937.4,4949
XS Rating Curve= 0 ,0
Exp/Cntr=0.3,0.1

Type RM Length L Ch R = 1 ,30256   ,121,121,121
BEGIN DESCRIPTION:
Mapping XS dd04a217
END DESCRIPTION:
XS GIS Cut Line= 4
3739057.50150913  10608498.44315      3738943.25     10608626.18
      3738666.55     10608807.04      3738593.95     10608874.57
#Sta/Elev= 30
  4649.6  335.25  4663.8  334.34  4713.1  335.51  4805.1  332.75  4812.6  331.45
  4834.4  329.79  4840.3  328.13  4849.2  327.25  4855.5  323.44  4885.1  316.97
  4912.7  314.22    4943  314.41  4964.1  312.93    4970  312.77  4979.2  310.72
  4985.1  311.08  4989.6  309.56  4992.3  309.06  4995.6  309.56  5000.3  313.25
  5006.2  311.74  5015.4  316.27  5021.3  316.81  5078.6  318.93  5087.8  318.35
  5129.9  322.67    5145     322  5222.4  326.26  5229.3  325.78  5250.7  328.44
#Mann= 3 ,-1 , 0
  4649.6     .16       0  4989.6     .07       0  4995.6     .16       0
Bank Sta=4964.1,5000.3
XS Rating Curve= 0 ,0
Exp/Cntr=0.3,0.1

Type RM Length L Ch R = 1 ,30135   ,61,61,61
BEGIN DESCRIPTION:
Mapping XS 54bb4b5d
END DESCRIPTION:
XS GIS Cut Line= 4
3738902.5346644510608392.5886286      3738782.43     10608542.33
      3738708.21     10608650.79      3738613.65     10608798.66
#Sta/Elev= 30
  4661.9  337.05  4676.3   336.1  4769.1  335.98  4797.9   333.7  4818.7  334.54
  4839.5  332.82  4847.5  331.77  4852.1  329.85  4868.6  329.34  4875.5  327.46
  4883.5  322.83  4898.4  319.24  4904.5  318.92  4911.8  316.32  4948.2  312.64
  4970.2  311.48  4976.2   310.8  4978.9  307.35  4981.6  306.85  4984.9  307.35
  5006.4  311.58  5033.5  312.76  5042.8  313.61  5048.7  315.21    5064  315.53
  5085.1   318.1  5100.3  318.14  5127.4  320.91  5157.8  322.43  5160.8  323.61
#Mann= 3 ,-1 , 0
  4661.9     .16       0  4978.9     .07       0  4984.9     .16       0
Bank Sta=4970.2,5006.4
XS Rating Curve= 0 ,0
Exp/Cntr=0.3,0.1

Type RM Length L Ch R = 1 ,30074   ,118,118,118
BEGIN DESCRIPTION:
Mapping XS b9113b89
END DESCRIPTION:
XS GIS Cut Line= 3
3738804.53977625 10608365.043061      3738654.39     10608610.86
       3738602.3      10608774.1
#Sta/Elev= 30
  4669.9  336.92  4685.4  337.28  4691.2  336.56  4706.7  336.14  4743.4  336.16
    4758  335.38  4780.2  335.88  4786.1  334.45  4844.1     332  4851.7  330.11
  4865.4  329.52  4880.9  327.22  4886.8  324.82  4902.2  322.51  4910.3   319.3
  4933.1  316.22  4957.7  313.29  4986.8  313.43  4992.1  311.15  4999.2  309.13
  5009.7  310.43    5019  315.43  5030.7  316.97  5062.2  318.06  5083.2   319.5
  5093.9  318.77  5104.2  320.53  5114.7  320.64  5120.8  322.01  5129.3  321.37
#Mann= 3 ,-1 , 0
  4669.9     .16       0  4986.8     .07       0    5019     .16       0
Bank Sta=4986.8,5019
XS Rating Curve= 0 ,0
Exp/Cntr=0.3,0.1

Type RM Length L Ch R = 1 ,29956   ,127,127,127
BEGIN DESCRIPTION:
MACK CREEK 60.0
END DESCRIPTION:
XS GIS Cut Line= 3
3738706.4363534910608378.3499494      3738599.61     10608560.19
      3738549.61     10608860.15
#Sta/Elev= 30
  4808.8  335.59  4822.5  334.41    4836  335.53  4857.5  335.65  4880.5  334.68
  4888.8  333.47  4916.1  333.94  4931.8  332.58  4947.5  329.55  4953.3  318.75
  4968.9  314.73  4974.7  312.38  4984.6  310.67  4987.4   309.3  4990.1   308.8
  4993.4   309.3  5011.9  311.34  5029.8  311.54    5040  312.58  5052.6  315.18
  5060.2  315.65  5070.4  316.83  5080.5  316.55  5090.7  317.44  5108.4  316.44
  5131.2  317.47  5181.9  317.84  5202.2  319.81  5235.1  321.12  5323.8  328.75
#Mann= 3 ,-1 , 0
  4808.8     .16       0  4987.4     .07       0  4993.4     .08       0
Bank Sta=4968.9,5060.2
XS Rating Curve= 0 ,0
Exp/Cntr=0.3,0.1

Type RM Length L Ch R = 1 ,29829   ,361,361,361
BEGIN DESCRIPTION:
Mapping XS 4d929c8c
END DESCRIPTION:
XS GIS Cut Line= 3
3738522.8791320410608390.1839363      3738505.09     10608581.35
      3738501.62     10608843.53
#Sta/Elev= 30
  4920.2  331.73  4940.3  333.64  4950.3  333.28  4960.4  329.46  4970.4  318.71
  4980.5  314.71  4990.5  306.86  5000.6  307.94  5007.5  313.56  5020.6  314.15
  5030.7   314.1  5070.9   312.3  5080.9  312.29    5141  313.59  5147.2  314.72
  5152.2  314.16    5211  313.88    5221   312.7    5231  312.59    5241  313.75
    5251  315.83    5261   317.3    5271  317.56  5291.1  318.96  5301.1  320.63
  5321.1   322.9  5341.1  324.44  5351.1  326.09  5370.2  327.73  5374.4  327.73
#Mann= 3 ,-1 , 0
  4920.2     .16       0  4980.5     .07       0  5007.5     .08       0
Bank Sta=4980.5,5007.5
XS Rating Curve= 0 ,0
Exp/Cntr=0.3,0.1

Type RM Length L Ch R = 1 ,29468   ,222,222,222
BEGIN DESCRIPTION:
Mapping XS 6ff16cb9
END DESCRIPTION:
XS GIS Cut Line= 4
        3738422.       10608357.      3738415.45     10608457.26
      3738413.07     10608553.57      3738430.44     10608850.45
#Sta/Elev= 30
  4614.4  330.39  4684.5  328.57  4694.5  327.58  4704.5  327.25  4710.5  326.15
  4715.5  326.15  4734.5  324.69  4774.5   320.9  4794.5  319.38  4807.9  318.91
  4814.5  317.78  4824.6  317.32  4831.9  316.42  4836.9  316.93  4874.6  315.08
  4884.7  315.62  4894.7   315.6  4904.7  314.61  4934.7  312.89  4964.8  311.85
  4984.8  311.69  4994.8  310.58  5002.7  308.83  5007.7  308.36  5014.9  306.62
  5024.9  309.81  5034.9     317    5055   324.1    5065  326.34  5105.3  328.72
#Mann= 2 ,-1 , 0
  4614.4     .16       0  5002.7     .07       0
Bank Sta=4984.8,5024.9
XS Rating Curve= 0 ,0
Exp/Cntr=0.3,0.1

Type RM Length L Ch R = 1 ,29246   ,327,327,327
BEGIN DESCRIPTION:
MACK CREEK 59.0
END DESCRIPTION:
XS GIS Cut Line= 3
3738348.3633617510608340.2123977      3738352.59     10608488.23
      3738161.64     10608814.59
#Sta/Elev= 30
    4702  325.49    4712  324.91    4732  325.29    4782   323.6    4812  320.93
  4898.7  315.26  4910.8  315.43  4926.5  313.95  4979.4  312.38  4985.1  312.95
  4988.4  301.22  4991.1  300.72  4994.4  301.22  5006.6  303.46  5014.6  308.62
  5022.3  309.35  5028.1  311.21  5037.7  312.27  5043.8   315.5  5065.3  318.77
  5072.5  317.05    5081  316.44  5086.8  322.01  5095.7  323.13  5102.5  327.62
  5166.9  334.29  5182.6  335.41  5204.1  335.82  5211.5  336.95  5228.2  337.08
#Mann= 3 ,-1 , 0
    4702     .16       0  4988.4     .07       0  4994.4     .16       0
Bank Sta=4979.4,5037.7
XS Rating Curve= 0 ,0
Exp/Cntr=0.3,0.1

Type RM Length L Ch R = 1 ,28919   ,381,381,381
BEGIN DESCRIPTION:
MACK CREEK 58.0
END DESCRIPTION:
XS GIS Cut Line= 2
      3738043.56     10608092.42      3737963.71     10608783.32
#Sta/Elev= 30
  4617.4  326.53  4635.3   326.5  4675.6   322.9    4693  319.07    4698  323.37
  4705.8  319.62  4725.9  319.73    4736  321.16  4776.2  319.29  4796.4     321
  4826.6  319.65  4856.8  315.49  4870.7  315.83  4927.2  310.51  4977.6  310.59
  4997.7   307.6  5007.8  299.13  5014.8  298.97  5017.6  298.47  5020.8  298.97
  5027.9  309.12  5068.2  311.47  5078.2  316.56  5088.3  318.32  5108.4  321.67
  5132.2  322.81  5138.6  324.66  5158.7  327.21  5239.3  333.84  5312.9  336.09
#Mann= 3 ,-1 , 0
  4617.4     .16       0  5014.8     .07       0  5020.8     .16       0
Bank Sta=4997.7,5027.9
XS Rating Curve= 0 ,0
Exp/Cntr=0.3,0.1

Type RM Length L Ch R = 1 ,28538   ,506,506,506
BEGIN DESCRIPTION:
MACK CREEK 57.0
END DESCRIPTION:
XS GIS Cut Line= 3
      3737749.61     10608260.18      3737699.61     10608389.36
      3737649.61     10608660.16
#Sta/Elev= 30
    4807  319.76  4851.9   319.2  4860.6  316.86  4876.5   315.4  4882.1  312.68
  4892.8  311.41  4901.1  308.67  4914.2  308.39    4931  309.71  4948.5  309.72
  4966.7  308.43  4972.4  303.62  4977.5  307.98  4997.2  302.78  5007.4  298.67
  5017.5  298.99  5025.4  300.51  5027.5   297.9  5030.2   297.4  5033.5   297.9
  5037.9  300.57  5048.1  307.23  5058.2  308.89  5083.4  308.58  5088.7  310.56
  5136.4  314.03  5159.9  318.05  5194.4  320.87  5200.6  322.51  5220.9  324.86
#Mann= 3 ,-1 , 0
    4807     .16       0  5027.5     .07       0  5033.5     .16       0
Bank Sta=5025.4,5037.9
XS Rating Curve= 0 ,0
Exp/Cntr=0.3,0.1

Type RM Length L Ch R = 1 ,28032   ,397,397,397
BEGIN DESCRIPTION:
MACK CREEK 56.0
END DESCRIPTION:
XS GIS Cut Line= 3
      3737480.68     10607995.32      3737315.73      10608333.9
      3737172.55     10608685.33
#Sta/Elev= 30
    4800   327.2  4827.7  327.05    4835   325.6  4849.9  325.87  4885.6  323.84
  4902.6  321.39  4908.1  322.56  4925.1   319.1  4930.7   319.2  4938.9     316
  4953.2  313.08  4970.2  308.24  4975.8  308.34  5005.6  302.79  5012.3  299.56
    5015  299.06  5018.3  299.56  5037.8  303.17  5043.4  307.12    5111  306.24
  5194.2  309.03  5202.8  308.11  5237.7  307.93  5363.3  311.42  5410.2  314.82
  5422.2  317.07  5440.9  318.36  5485.8  323.26  5499.8  325.95  5556.1  331.97
#Mann= 3 ,-1 , 0
    4800     .16       0  5012.3     .07       0  5018.3     .16       0
Bank Sta=5005.6,5037.8
XS Rating Curve= 0 ,0
Exp/Cntr=0.3,0.1

Type RM Length L Ch R = 1 ,27635   ,492,492,492
BEGIN DESCRIPTION:
MACK CREEK 55.0
END DESCRIPTION:
XS GIS Cut Line= 3
       3737099.6     10608060.24      3737049.61     10608289.36
      3737049.61     10608560.15
#Sta/Elev= 30
  4755.8  322.74  4780.3  321.48  4786.5  319.33  4796.7  318.45  4817.2  315.01
  4824.2  311.47  4829.3  312.15  4847.9  307.61  4873.2   305.9  4909.3  306.61
  4917.2  305.65  4929.7  305.83  4971.3  304.17  4993.2  305.15  5001.1  303.17
  5011.1  297.37  5018.1  295.55  5020.9  295.05  5024.1  295.55  5031.1  296.49
  5041.1   299.9  5051.1  305.74  5061.1  307.27  5071.1  306.34  5111.1  305.32
  5141.1  307.09  5171.1   311.2  5181.1  311.78  5201.1  315.16  5261.1  322.12
#Mann= 3 ,-1 , 0
  4755.8     .16       0  5018.1     .07       0  5024.1     .16       0
Bank Sta=5001.1,5051.1
XS Rating Curve= 0 ,0
Exp/Cntr=0.3,0.1

Type RM Length L Ch R = 1 ,27143   ,410,410,410
BEGIN DESCRIPTION:
MACK CREEK 54.0
END DESCRIPTION:
XS GIS Cut Line= 3
      3736899.64     10607910.15      3736649.61     10608289.36
      3736549.61     10608660.19
#Sta/Elev= 30
  4536.2  326.89  4598.4  323.62  4644.1  316.01  4658.2   315.2    4680   309.5
  4688.3   305.9  4838.8  305.75  4853.9   310.8  4859.9  308.14    4869  313.83
  4883.6  313.91    4896  313.27  4926.2  305.37  4942.1  304.93  4955.5  304.73
  4962.3  302.23  4968.3  304.01  4983.4  304.37  4993.4  302.97  5010.4  294.08
  5013.1  293.58  5016.4  294.08  5032.7  300.78  5053.4  302.73    5128  304.99
  5162.7  310.44  5208.8  313.67  5229.5  315.99  5237.4   318.4  5374.5  333.47
#Mann= 5 ,-1 , 0
  4536.2     .16       0  4598.4     .05       0  4942.1     .16       0
  5010.4     .07       0  5016.4     .16       0
Bank Sta=4993.4,5032.7
XS Rating Curve= 0 ,0
Exp/Cntr=0.3,0.1

Type RM Length L Ch R = 1 ,26733   ,559,559,559
BEGIN DESCRIPTION:
MACK CREEK 53.0
END DESCRIPTION:
XS GIS Cut Line= 3
      3736849.62     10607710.17      3736299.61     10608489.36
      3736299.61      10608610.2
#Sta/Elev= 30
  4081.1  333.11  4325.9  322.29    4368  322.17  4380.6  319.26  4388.9  319.95
  4397.6  316.85  4411.6     316  4418.5  312.69    4469  305.84  4656.2  306.17
  4668.7  311.03    4698  313.61  4712.8  312.54  4748.5  304.85  4819.9  302.82
    4848  301.61  4897.6  302.53  4957.2  303.16  5013.2  303.58  5021.8  297.65
    5028  298.33  5029.3  291.16  5032.1  290.66  5035.3  291.16  5045.7  291.42
  5055.7  296.65  5065.7  298.26  5095.7  316.35  5135.7   329.8  5155.7  333.32
#Mann= 7 ,-1 , 0
  4081.1     .16       0  4380.6     .05       0    4848     .16       0
  4897.6     .12       0  4957.2     .16       0  5029.3     .07       0
  5035.3     .16       0
Bank Sta=4819.9,5065.7
XS Rating Curve= 0 ,0
Exp/Cntr=0.3,0.1

Type RM Length L Ch R = 1 ,26174   ,336,336,336
BEGIN DESCRIPTION:
MACK CREEK 52.0
END DESCRIPTION:
XS GIS Cut Line= 3
      3736482.41     10607669.82      3736026.67     10608090.84
      3735809.66     10608394.65
#Sta/Elev= 30
  4300.5  321.87  4414.1  315.88  4472.5  312.45  4479.9  310.84  4500.9  310.54
  4557.6  305.27  4635.2  301.12    4777  300.01    4883  302.26  4911.4  300.76
    4921  298.83  4925.4  296.36    4961  299.73  4981.9  299.45  5005.3  294.67
  5008.4  288.75  5011.2  288.25  5014.4  288.75  5018.5  288.85  5026.2  295.58
  5040.9  299.86  5061.8   309.3  5082.7  310.37  5091.3  312.45  5147.8  319.45
  5168.7  320.49  5190.5  325.04  5227.4  328.69  5276.5  336.01  5294.3  336.81
#Mann= 4 ,-1 , 0
  4300.5     .16       0  4414.1     .12       0  5008.4     .07       0
  5014.4     .16       0
Bank Sta=5005.3,5026.2
XS Rating Curve= 0 ,0
Exp/Cntr=0.3,0.1

Type RM Length L Ch R = 1 ,25838   ,473,473,473
BEGIN DESCRIPTION:
MACK CREEK 51.0
END DESCRIPTION:
XS GIS Cut Line= 3
      3736499.62     10607260.17      3735699.61     10607989.36
      3735599.62     10608060.18
#Sta/Elev= 30
  3947.9  344.78  4057.1   337.9  4089.4  335.14  4229.1   324.5  4372.6  312.69
  4584.7  298.99  4627.3  298.82  4655.7  301.48  4769.2  296.41  4861.1  298.02
    4868  293.57  4875.2     293  4903.6  293.43  4915.8  295.78    4932  298.17
    4953  297.73  4960.4  295.02  4981.3   295.2  4988.7  292.62  4995.5  294.53
  5006.7  287.44  5009.5  286.94  5012.7  287.44  5023.9  290.57  5027.3  295.77
  5053.3  302.22  5067.1  303.62  5080.3  312.46  5145.5  322.18  5152.9  321.67
#Mann= 7 ,-1 , 0
  3947.9     .16       0  4057.1     .12       0  4089.4     .16       0
  4229.1     .12       0  4915.8     .16       0  5006.7     .07       0
  5012.7     .16       0
Bank Sta=4995.5,5027.3
XS Rating Curve= 0 ,0
Exp/Cntr=0.3,0.1

Type RM Length L Ch R = 1 ,25365   ,552,552,552
BEGIN DESCRIPTION:
MACK CREEK 50.0
END DESCRIPTION:
XS GIS Cut Line= 3
      3736030.99     10607335.64      3735592.64     10607626.43
      3735375.63     10607960.63
#Sta/Elev= 30
  4398.9  324.12  4504.6  318.64  4576.8  305.32  4640.6  299.63  4727.1  297.93
  4757.2  294.35  4799.3  296.69  4808.4  291.98  4814.4  295.37  4835.4  297.05
  4865.5  295.21  4871.5  296.43  4916.6  296.03  4922.6  294.35  4952.7  296.13
  4958.6  293.91  4988.9   295.9  4994.9  286.18    5007  285.13  5009.8  284.63
    5013  285.13  5031.1  286.17  5037.1  292.28  5046.3  298.18  5052.2  304.32
  5088.5  308.95  5290.8   326.5    5299  326.65    5306  324.02  5323.4  325.26
#Mann= 3 ,-1 , 0
  4398.9     .16       0    5007     .07       0    5013     .16       0
Bank Sta=4988.9,5037.1
XS Rating Curve= 0 ,0
Exp/Cntr=0.3,0.1

Type RM Length L Ch R = 1 ,24813   ,322,322,322
BEGIN DESCRIPTION:
MACK CREEK 49.0
END DESCRIPTION:
XS GIS Cut Line= 3
      3735883.86     10607040.29      3735425.51     10607418.78
       3735099.1     10607981.31
#Sta/Elev= 30
  4296.2  315.87  4369.9  313.05  4491.1  300.59  4554.9  297.13  4789.4  295.21
  4824.6   297.2  4887.8  294.04    4911  295.31  4932.5   292.8  4975.5  295.63
    5007  290.46  5009.8  283.34  5012.6  282.84  5015.8  283.34  5028.6  284.53
  5034.3   289.7  5042.6  290.29  5050.1  287.29  5055.9   290.9  5065.7  286.37
  5071.6  292.19  5077.4  291.59  5100.4  300.72  5108.9  302.15  5210.7   309.8
  5387.1  322.03  5451.7  323.06  5504.7  327.37  5510.4  325.04    5541  327.77
#Mann= 3 ,-1 , 0
  4296.2     .16       0  5009.8     .07       0  5015.8     .16       0
Bank Sta=5007,5034.3
XS Rating Curve= 0 ,0
Exp/Cntr=0.3,0.1

Type RM Length L Ch R = 1 ,24491   ,457,457,457
BEGIN DESCRIPTION:
MACK CREEK 48.0
END DESCRIPTION:
XS GIS Cut Line= 3
      3735803.94     10607022.97      3735415.09     10607224.34
       3734529.7     10607387.53
#Sta/Elev= 30
  4508.3  308.11    4516   308.7  4576.7  303.32  4582.4   303.8  4598.9  301.03
  4643.1  299.67  4670.9  297.08  4703.9   295.6  4731.7  296.69  4748.2  295.41
  4792.5  295.16  4814.6  296.51  4903.1  289.75  4925.3  291.32  4961.9  291.33
  4972.1   287.9  4989.4  283.95  4992.2  283.45  4995.4  283.95  5006.9  284.09
  5012.8  289.83  5043.3  292.59  5195.8  313.45    5224  316.39  5340.2  317.98
  5446.2   316.8  5551.7  318.53  5795.8  326.21  5837.6  329.02  5846.5  328.12
#Mann= 3 ,-1 , 0
  4508.3     .16       0  4989.4     .07       0  4995.4     .16       0
Bank Sta=4961.9,5012.8
XS Rating Curve= 0 ,0
Exp/Cntr=0.3,0.1

Type RM Length L Ch R = 1 ,24034   ,520,520,520
BEGIN DESCRIPTION:
MACK CREEK 47.0
END DESCRIPTION:
XS GIS Cut Line= 3
      3735699.63     10606860.19      3735299.61     10606889.36
      3735099.57     10606910.19
#Sta/Elev= 30
  4610.3  299.77  4670.5  296.22  4740.7  295.07  4790.8  291.74  4810.9  291.93
  4816.2  293.93  4821.2  292.89  4830.9  293.73    4861  290.23  4891.1  293.03
  4901.1  292.98  4921.1  289.85  4961.2  291.69  4971.3  285.35  4981.3  282.26
  4988.3  281.95  4991.1  281.45  4994.3  281.95  5008.9  285.73  5041.5  290.56
  5051.6  287.07  5067.2  284.36  5081.8  286.79  5101.9  287.83  5111.9  292.44
  5142.1  297.68  5160.7  302.61  5165.7  302.18  5172.2  304.29  5212.5   310.7
#Mann= 3 ,-1 , 0
  4610.3     .16       0  4988.3     .07       0  4994.3     .16       0
Bank Sta=4971.3,5008.9
XS Rating Curve= 0 ,0
Exp/Cntr=0.3,0.1

Type RM Length L Ch R = 1 ,23514   ,464,464,464
BEGIN DESCRIPTION:
MACK CREEK 46.0
END DESCRIPTION:
XS GIS Cut Line= 3
      3735699.59     10605760.21      3735049.61     10606539.36
      3734749.62     10606610.19
#Sta/Elev= 30
  3960.2  326.88  4158.7   304.3  4592.1  294.14  4641.6  291.31    4691   291.7
  4698.8   286.2  4705.3  288.22  4719.6   281.3    4734  278.39  4741.5  290.12
  4754.8  291.57  4797.7  288.06  4805.5  289.57  4812.1  287.68  4826.4  290.13
  4918.8  288.49  4947.4  284.33  4953.9  280.22  4961.7  283.29  4968.3   277.5
  4972.2  283.05  4974.9  283.05  4992.3  274.88    4995  274.38  4998.3  274.88
  5026.2   283.8  5042.7  289.24  5132.5  294.01  5211.2  305.09  5283.1  311.03
#Mann= 3 ,-1 , 0
  3960.2     .16       0  4992.3     .07       0  4998.3     .16       0
Bank Sta=4974.9,5026.2
XS Rating Curve= 0 ,0
Exp/Cntr=0.3,0.1

Type RM Length L Ch R = 1 ,23050   ,529,529,529
BEGIN DESCRIPTION:
MACK CREEK 45.0
END DESCRIPTION:
XS GIS Cut Line= 3
      3735099.59     10605860.21      3734799.61     10606239.36
      3734749.61     10606560.21
#Sta/Elev= 30
  4487.6  297.61  4736.8  288.69  4829.8  287.79    4865  286.44  4871.4  287.23
  4914.7  285.58    4958  286.42  4964.4  285.54  4968.4   283.5    4974   283.5
  4992.2  273.41  5000.4  273.65  5002.4  272.44  5005.2  271.94  5008.4  272.44
  5012.4  277.22  5032.6  285.53  5042.8  286.69  5068.3  287.29  5174.3  287.54
    5199  289.87  5204.7  292.14  5214.8  293.64  5224.9  296.88  5235.1  297.62
  5245.2  300.03  5255.3  300.88  5261.8  302.81  5266.9  302.56  5295.8  306.57
#Mann= 3 ,-1 , 0
  4487.6     .16       0  5002.4     .07       0  5008.4     .16       0
Bank Sta=4974,5032.6
XS Rating Curve= 0 ,0
Exp/Cntr=0.3,0.1

Type RM Length L Ch R = 1 ,22521   ,446,446,446
BEGIN DESCRIPTION:
MACK CREEK 44.0
END DESCRIPTION:
XS GIS Cut Line= 3
      3734799.63     10605660.16      3734549.61     10606039.36
      3734349.63     10606460.15
#Sta/Elev= 30
  4559.1  308.43  4679.3  299.24  4789.5  290.13  4840.7  283.94  4912.9  283.68
  4918.9  282.71  4949.8  283.27  4972.3  285.25  4985.2  284.26  4991.2  281.72
  5000.3  274.33  5003.3  270.05    5006  269.55  5009.3  270.05  5010.8  272.15
  5016.5  272.15  5022.4  277.11  5027.9  279.88  5036.4  281.19  5050.6  283.04
  5067.8  282.76  5073.3  283.91  5080.7   282.2    5096  284.46  5202.4  284.14
  5328.8  288.09    5435  295.54  5442.4  297.55  5447.9  297.22  5479.2  300.87
#Mann= 6 ,-1 , 0
  4559.1     .12       0  4679.3     .16       0  4949.8     .05       0
  4972.3     .16       0  5003.3     .07       0  5009.3     .16       0
Bank Sta=4991.2,5036.4
XS Rating Curve= 0 ,0
Exp/Cntr=0.3,0.1

Type RM Length L Ch R = 1 ,22075   ,334,334,334
BEGIN DESCRIPTION:
MACK CREEK 43.0
END DESCRIPTION:
XS GIS Cut Line= 3
      3734399.63     10605560.17      3734299.61     10605689.36
      3733999.61     10606110.19
#Sta/Elev= 30
  4812.6   294.4  4826.2  292.53  4863.2  290.47  4898.7  285.66    4906  283.34
  4919.5  281.56  4948.4  282.78    4990  281.35  4998.6  278.46  5010.4  267.71
  5013.1  267.21  5016.4  267.71  5019.5  269.04  5026.1  270.44  5034.3  278.88
  5040.4  280.77    5049  281.39    5063  283.73  5069.9  282.26  5076.1  281.95
  5120.3  282.25  5126.5  281.39    5156   282.8  5307.2  281.39  5393.2  282.52
    5435  284.13  5443.6  283.89  5485.4  286.32  5489.7  287.56  5492.8  287.56
#Mann= 4 ,-1 , 0
  4812.6     .12       0    4906     .16       0  5010.4     .07       0
  5016.4     .16       0
Bank Sta=4990,5040.4
XS Rating Curve= 0 ,0
Exp/Cntr=0.3,0.1

Type RM Length L Ch R = 1 ,21741   ,537,537,537
BEGIN DESCRIPTION:
MACK CREEK 42.0
END DESCRIPTION:
XS GIS Cut Line= 3
       3734276.2      10605241.7      3733949.82     10605672.25
      3733918.61     10606195.85
#Sta/Elev= 30
    4670  306.94  4702.6  303.52  4708.9  304.25  4738.8  301.73  4773.4  299.95
  4787.9     297  4808.7  296.37  4873.2  289.63  4881.4  286.42    4894  284.22
  4908.6  280.74  4937.7  279.65  4958.5  275.08  4981.3  275.55  4987.6  271.85
  4994.4  274.19  5002.2  273.22  5008.4  267.71    5020  266.93  5022.7  266.43
    5026  266.93  5031.3  270.48  5037.5  283.15  5069.7  282.91  5230.1   281.1
  5438.6  281.36  5548.8  283.65  5628.9  288.27  5709.1  298.33  5734.8  299.87
#Mann= 7 ,-1 , 0
    4670     .16       0  4738.8     .12       0    4894     .16       0
    5020     .07       0    5026     .16       0  5069.7     .12       0
  5230.1     .16       0
Bank Sta=5002.2,5037.5
XS Rating Curve= 0 ,0
Exp/Cntr=0.3,0.1

Type RM Length L Ch R = 1 ,21204   ,271,271,271
BEGIN DESCRIPTION:
MACK CREEK 41.0
END DESCRIPTION:
XS GIS Cut Line= 3
      3733790.09     10604981.31      3733717.18     10605620.17
      3733845.58     10606345.49
#Sta/Elev= 30
  4561.2  298.97  4650.7  295.86  4660.7  295.95  4680.8  298.84  4690.9  296.81
  4721.1  285.48  4761.4  280.48  4801.6  277.76  4831.8  277.17  4851.9  280.03
  4932.5  279.82    4960  277.92    4965  275.44  4972.7  272.95  5002.9  269.77
    5013  267.63  5022.8  263.89  5026.1  264.39  5043.2  272.98  5049.3  274.39
  5054.4  277.88    5534  284.71  5706.3  293.55  5752.6  296.82  5760.4  298.28
  5765.5  297.74  5783.1  299.88  5803.4  300.48    5844   304.9  5940.8  311.56
#Mann= 1 ,-1 , 0
  4561.2     .16       0
Bank Sta=4965,5054.4
XS Rating Curve= 0 ,0
Exp/Cntr=0.3,0.1

Type RM Length L Ch R = 1 ,20933   ,513,513,513
BEGIN DESCRIPTION:
MACK CREEK 40.0
END DESCRIPTION:
XS GIS Cut Line= 3
      3733578.28     10604897.99      3733512.32     10605415.31
      3732953.95     10605994.48
#Sta/Elev= 30
  4622.6  312.29  4725.6  298.59  4735.7  292.48    4776  286.75    4897  279.84
  4907.1  270.49  4917.2  268.62  4937.3  271.77  4965.2  269.92  4970.2  273.14
  4997.6  262.45  5028.1  274.08  5098.6  278.03  5118.8  277.09  5129.9  270.43
    5144  276.02  5163.7   277.3  5241.4  277.54  5276.7  275.48  5283.9  266.26
    5305  265.51  5312.2   268.7  5319.1   265.7  5326.3  278.26  5340.5  279.57
  5573.8  285.31  5602.1  292.07  5637.3  291.52  5771.9  308.01  5948.6  311.43
#Mann= 1 ,-1 , 0
  4622.6     .16       0
#XS Ineff= 2 , 0
       0                 5097.95       0     290
Permanent Ineff=
       F       F
Bank Sta=4970.2,5028.1
XS Rating Curve= 0 ,0
Exp/Cntr=0.3,0.1

Type RM Length L Ch R = 1 ,20420   ,480,480,480
BEGIN DESCRIPTION:
Mapping XS 8b3f9f13
END DESCRIPTION:
XS GIS Cut Line= 3
      3733512.29     10604665.35      3733363.01       10604891.
      3732666.23     10605546.19
#Sta/Elev= 30
  4655.8  317.48  4668.7  318.26  4674.7  316.24  4755.9  309.77    4792  304.98
    4798     302  4813.1  302.82  4819.1  300.44  4849.2  297.62  4855.2  294.57
  4900.4  285.09  4906.4  280.02  4924.9  273.33  4970.8   266.8  4977.7  268.39
    4985  261.64  5026.9  258.72  5030.1  259.22  5034.3  272.21  5041.2  268.92
  5048.5  273.45  5076.8  276.42  5175.9  273.91  5359.6  275.72  5381.1  273.57
  5614.5  277.05  5635.6   279.9    5657  278.56  5755.7  286.78  5882.8  300.42
#Mann= 1 ,-1 , 0
  4655.8     .16       0
#XS Ineff= 2 , 0
       0                 5068.52       0     290
Permanent Ineff=
       F       F
Bank Sta=4977.7,5034.3
XS Rating Curve= 0 ,0
Exp/Cntr=0.3,0.1

Type RM Length L Ch R = 1 ,19940   ,482,482,482
BEGIN DESCRIPTION:
Mapping XS c49f60c5
END DESCRIPTION:
XS GIS Cut Line= 3
       3733126.9     10604456.97      3733067.87     10604835.45
      3732519.27     10605394.47
#Sta/Elev= 30
  4781.6  315.63  4798.3  314.43  4805.1  311.71  4855.7  303.65  4861.1   301.1
  4875.9  299.95  4896.2  294.84  4916.4  282.59  4923.9   279.7  4928.9  279.91
  4936.7  274.43  4946.8  273.43  4956.9  268.77  4986.7  259.37  4991.7  261.62
  4994.4  256.84  4997.1  256.34  5000.4  256.84  5007.5  256.89  5027.8  267.74
  5037.9  273.84  5054.6  274.73  5272.8  274.17  5322.4  272.73  5421.4  273.87
    5584  271.54  5718.3   273.4    5789  277.16  5810.3  280.77  5947.9  295.89
#Mann= 3 ,-1 , 0
  4781.6     .16       0  4994.4     .07       0  5000.4     .16       0
#XS Ineff= 2 , 0
                          5281.7          279.09
Permanent Ineff=
       F       F
Bank Sta=4956.9,5027.8
XS Rating Curve= 0 ,0
Exp/Cntr=0.3,0.1

Type RM Length L Ch R = 1 ,19458   ,434,434,434
BEGIN DESCRIPTION:
MACK CREEK 37.0
END DESCRIPTION:
XS GIS Cut Line= 3
      3732849.62     10604410.18      3732649.61     10604639.36
      3732249.63     10605010.17
#Sta/Elev= 30
  4684.1  314.15  4740.6  307.84  4890.4  279.84  4932.4  273.42  4946.6  265.79
  4963.7   264.5  4967.5  264.45  4999.8  255.53  5002.5  255.03  5005.8  255.53
  5010.2  260.07  5019.1  261.51  5031.1  268.81  5137.7   270.9  5151.9  265.12
  5172.9  263.02  5179.7  268.79  5193.9  270.45  5201.2  266.75  5215.4  268.31
  5222.2  265.69  5236.4  268.21  5243.7  273.03  5335.6  277.49  5342.8  273.51
  5356.6   273.8  5363.9  277.57  5384.9  275.81  5525.9  287.95  5533.7  289.58
#Mann= 7 ,-1 , 0
  4684.1      .1       0  4890.4     .16       0  4963.7      .1       0
  4999.8     .07       0  5005.8      .1       0  5019.1     .16       0
  5525.9     .05       0
#XS Ineff= 2 , 0
                         5136.36          278.47
Permanent Ineff=
       F       F
Bank Sta=4967.5,5031.1
XS Rating Curve= 0 ,0
Exp/Cntr=0.3,0.1

Type RM Length L Ch R = 1 ,19024   ,419,419,419
BEGIN DESCRIPTION:
MACK CREEK 36.0
END DESCRIPTION:
XS GIS Cut Line= 3
      3732649.64     10604260.16      3732249.61     10604589.36
       3732149.6      10604810.2
#Sta/Elev= 30
  4467.7  284.51  4532.3  280.98  4538.8  281.65  4553.1   279.7  4573.9  279.34
  4581.8  277.72  4718.2  272.62  4840.4  270.02  4843.7  269.79  4851.5  264.49
  4853.3  265.57    4858  268.39  4865.9  267.22  4872.4  270.71  4921.9  268.59
  4936.2  267.77  4944.1   261.3  4950.6   260.6  4956.7  258.82    4989  256.17
    4992  254.36  4994.8  253.86    4998  254.36  5008.6  257.31  5018.1  264.93
  5046.7  265.81  5063.5  269.06  5069.8  271.99  5144.6   276.5  5228.2  285.61
#Mann= 7 ,-1 , 0
  4467.7     .16       0  4718.2      .1       0  4840.4     .16       0
  4853.3      .1       0  4956.7     .16       0    4992     .07       0
    4998     .16       0
Bank Sta=4950.6,5018.1
XS Rating Curve= 0 ,0
Exp/Cntr=0.3,0.1

Type RM Length L Ch R = 1 ,18605   ,496,496,496
BEGIN DESCRIPTION:
MACK CREEK 35.0
END DESCRIPTION:
XS GIS Cut Line= 3
      3732599.58     10603710.22      3731849.61     10604489.36
      3731849.61     10604810.22
#Sta/Elev= 30
  3926.6  319.75  4025.5  305.76  4032.7  303.06  4075.1  296.18  4145.9  287.04
    4289  277.56  4357.9  274.82  4591.5  271.67  4671.7  268.36  4725.8  265.89
  4803.4  266.78  4810.7  266.01  4814.5  262.79  4817.6  260.16  4824.8  261.46
  4831.7  258.37  4845.9  259.63    4860  265.93  4966.3  266.01  4980.5  249.88
  4987.4  246.65  4998.5   244.8  5001.3   244.3  5004.5   244.8  5005.1  253.52
    5011  253.52  5018.9  258.18  5038.9  265.18    5149  275.11  5328.9  291.47
#Mann= 7 ,-1 , 0
  3926.6      .1       0    4289     .16       0  4671.7      .1       0
  4814.5     .16       0  4998.5     .07       0  5004.5     .16       0
    5149     .05       0
Bank Sta=4966.3,5038.9
XS Rating Curve= 0 ,0
Exp/Cntr=0.3,0.1

Type RM Length L Ch R = 1 ,18109   ,383,383,383
BEGIN DESCRIPTION:
MACK CREEK 34.0
END DESCRIPTION:
XS GIS Cut Line= 3
      3731955.51     10603785.25      3731669.03     10604223.65
      3731565.29     10604586.72
#Sta/Elev= 30
  4632.9  271.55    4806  266.44  4835.8  266.59    4872  264.11  4877.9   265.9
  4887.1  261.97    4893   262.8  4901.6  258.82  4914.1  259.16  4923.3  264.63
  4929.2   259.4  4944.4  253.58  4950.3  255.22  4959.5  252.26  4965.4   256.5
  4973.3  253.48  4980.6  245.67  4986.5  242.72  4992.7  242.01  4995.4  241.51
  4998.7  242.01  5016.8  246.59  5031.9  253.01  5037.8  252.84    5053  258.63
  5058.9  259.26  5068.1  265.97  5282.4  266.66  5466.9  270.41  5534.2  272.03
#Mann= 4 ,-1 , 0
  4632.9     .16       0  4992.7     .07       0  4998.7     .16       0
  5466.9     .05       0
Bank Sta=4973.3,5031.9
XS Rating Curve= 0 ,0
Exp/Cntr=0.3,0.1

Type RM Length L Ch R = 1 ,17726   ,448,448,448
BEGIN DESCRIPTION:
Mapping XS 393b6878
END DESCRIPTION:
XS GIS Cut Line= 2
       3731529.4     10603660.17      3731227.34     10604384.08
#Sta/Elev= 30
  4706.7  267.61  4804.2  267.35  4824.8  266.17  4912.6  263.14  4927.9  260.06
  4934.3  255.44  4945.1   255.6  4957.1  253.08  4975.5  245.31    4996   241.1
  4996.3  241.06    4999  240.56  5002.3  241.06  5004.8  242.95    5021  247.59
  5028.6   251.3    5034  251.45  5064.3  261.15    5087  262.13  5110.9  261.08
  5140.1  263.05  5177.8  263.65  5302.7  265.22  5324.4  267.18  5341.5  266.71
  5346.9  268.24  5356.9  268.68  5378.5  266.85  5471.4  269.24  5491.1     268
#Mann= 6 ,-1 , 0
  4706.7     .05       0  4824.8      .1       0    4996     .16       0
  4996.3     .07       0  5002.3     .16       0  5177.8     .05       0
Bank Sta=4957.1,5028.6
XS Rating Curve= 0 ,0
Exp/Cntr=0.3,0.1

Type RM Length L Ch R = 1 ,17278   ,604,604,604
BEGIN DESCRIPTION:
Mapping XS e54ea61c
END DESCRIPTION:
XS GIS Cut Line= 2
      3731154.42      10603571.6      3730795.23     10604175.45
#Sta/Elev= 30
  4712.5  262.71  4780.7   259.9  4891.8  261.96  4920.3   260.2  4969.5  248.59
  4978.5  243.81  4993.8  239.96  5003.5  239.62  5006.3  239.12  5009.5  239.62
  5013.4  243.03    5028  247.68  5036.6   249.5  5049.4  249.03  5059.2  257.59
    5065  251.16  5071.6  257.66  5080.6  261.19  5086.4  259.06  5094.8  262.15
  5105.3   262.2  5187.9  261.38  5203.3  258.24  5218.9  261.12  5224.7  258.59
  5277.3  262.31  5303.7  261.98  5318.9  262.06  5394.1  262.48  5415.1  265.43
#Mann= 8 ,-1 , 0
  4712.5     .05       0  4891.8      .1       0  4993.8     .05       0
  5003.5     .04       0  5009.5     .05       0  5105.3     .08       0
  5303.7     .05       0  5318.9     .08       0
Bank Sta=4969.5,5028
XS Rating Curve= 0 ,0
Exp/Cntr=0.3,0.1

Type RM Length L Ch R = 1 ,16674   ,332,332,332
BEGIN DESCRIPTION:
MACK CREEK 31.0
END DESCRIPTION:
XS GIS Cut Line= 2
      3730774.94      10603216.7       3730171.6      10603859.1
#Sta/Elev= 30
  4661.8  276.61  4724.5  276.84  4760.1  273.56    4767  275.52  4837.8  274.99
    4852  272.33  4901.3  270.54  4915.4  268.05  4943.8  264.42  4951.1  256.61
    4958  254.98  4965.3  248.73  4972.1  245.05  4979.4  243.76  4990.6  237.39
  4993.4  236.89  4996.6  237.39  5014.6  240.53  5021.9  251.64  5036.1  257.32
  5050.3  257.99  5084.4  254.74  5205.6   260.9  5262.3  260.13  5269.6  262.15
  5401.9  267.35  5432.2  272.03  5460.5   269.4  5524.1  278.04  5543.1  278.67
#Mann= 6 ,-1 , 0
  4661.8     .05       0  4915.4     .16       0  4990.6     .07       0
  4996.6     .16       0  5084.4     .08       0  5401.9     .05       0
Bank Sta=4965.3,5021.9
XS Rating Curve= 0 ,0
Exp/Cntr=0.3,0.1

Type RM Length L Ch R = 1 ,16342   ,266,266,266
BEGIN DESCRIPTION:
MACK CREEK 30.0
END DESCRIPTION:
XS GIS Cut Line= 3
      3730499.65     10603160.17      3730299.61     10603239.36
      3729999.58     10603460.21
#Sta/Elev= 30
  4792.4  288.83  4807.3  288.25    4856  277.34  4891.1  273.46    4910  269.06
  4945.1   264.1  4953.8  262.52  4964.1  258.07  4969.5  260.47  4975.3  247.42
    4986  242.07  4993.8  236.59  5001.9  236.49  5004.6  235.99  5007.9  236.49
  5010.6  236.49  5015.6  240.82  5021.8  243.67  5030.2  243.96  5036.4  249.33
  5044.8  252.92  5075.9  256.31  5097.6  256.19  5222.3  258.33  5257.8  262.83
  5272.5  267.52  5283.3  268.05  5293.3  272.41  5328.7   275.1  5380.1  281.49
#Mann= 7 ,-1 , 0
  4792.4     .13       0  5001.9     .07       0  5007.9     .13       0
  5075.9     .05       0  5097.6     .08       0  5283.3     .05       0
  5328.7      .1       0
Bank Sta=4986,5021.8
XS Rating Curve= 0 ,0
Exp/Cntr=0.3,0.1

Type RM Length L Ch R = 1 ,16076   ,171,171,171
BEGIN DESCRIPTION:
Mapping XS afd32863
END DESCRIPTION:
XS GIS Cut Line= 3
      3730633.59     10602753.36      3730249.88     10602972.12
      3729768.95     10603241.24
#Sta/Elev= 30
  4438.3  281.81    4523  278.96  4746.4  279.66  4799.7  273.83  4811.2   266.7
  4857.3  258.55  4929.5  255.98  4937.6  253.82  4945.5  246.85  4972.9  242.52
  5001.9  235.25  5004.6  234.75  5007.9  235.25  5010.6  240.39  5017.8  243.14
  5032.3  247.52  5120.1  246.18  5143.9  246.71  5166.8  241.98  5172.7  246.82
  5210.4  247.76  5219.8  251.87  5297.2  253.66  5304.3  259.21  5327.2  264.13
  5362.3  265.94  5407.4  272.54  5415.9   276.5  5421.7  273.48  5431.1  275.83
#Mann= 6 ,-1 , 0
  4438.3     .05       0    4523     .16       0  5001.9     .07       0
  5007.9     .16       0  5120.1     .05       0  5219.8     .16       0
Bank Sta=4972.9,5017.8
XS Rating Curve= 0 ,0
Exp/Cntr=0.3,0.1

Type RM Length L Ch R = 1 ,15905   ,130,130,130
BEGIN DESCRIPTION:
Mapping XS 770d6008
END DESCRIPTION:
XS GIS Cut Line= 2
      3730388.81     10602613.25      3729795.91     10603135.94
#Sta/Elev= 30
  4615.4  277.52  4719.2  263.86    4761  252.61  4768.6  252.65  4775.3  259.71
  4832.2  264.09  4889.1  248.44  4966.9   245.9  4987.8  240.64  4992.3  234.63
  4995.1  234.13  4998.3  234.63  5023.8   241.9  5080.7  243.86  5101.6  247.92
  5150.9  244.48  5193.6  246.06  5207.8  250.57  5214.5   247.6    5222  253.47
  5228.7  252.03  5236.3  258.32  5242.9  255.88  5264.7  266.03  5271.4  263.89
    5279  270.21  5363.4  271.21  5377.6  274.31  5385.2  280.11  5405.8  279.76
#Mann= 3 ,-1 , 0
  4615.4     .13       0  4992.3     .07       0  4998.3     .13       0
Bank Sta=4987.8,5023.8
XS Rating Curve= 0 ,0
Exp/Cntr=0.3,0.1

Type RM Length L Ch R = 1 ,15775   ,150,150,150
BEGIN DESCRIPTION:
MACK CREEK 29.0
END DESCRIPTION:
XS GIS Cut Line= 4
      3730276.81     10602454.42      3730112.75     10602654.94
      3730026.81     10602878.89      3729773.11     10603101.53
#Sta/Elev= 30
  4648.3  264.76    4649  265.14    4718  263.72  4778.3  256.84  4812.9   257.2
  4870.9  254.18  4885.3  251.26  4891.7  245.25  4954.3  239.13  4954.8  237.92
  4956.6  233.56  4959.4  233.06  4962.6  233.56  4984.3  237.22  4989.6  233.95
  5037.4  235.73  5044.3  243.26  5058.3  241.01    5069  241.55  5074.3  248.01
  5093.7   247.7  5105.8  251.52  5116.5  247.28  5167.3   249.1  5202.8  246.19
  5280.7  255.86  5323.4  268.03  5422.9  271.81  5429.6  279.64  5484.8  287.09
#Mann= 10 ,-1 , 0
  4648.3     .16       0    4649     .08       0    4718     .16       0
  4812.9     .05       0  4954.8     .16       0  4956.6     .07       0
  4962.6     .16       0  5037.4     .05       0  5058.3     .08       0
  5167.3     .16       0
Bank Sta=4954.3,4984.3
XS Rating Curve= 0 ,0
Exp/Cntr=0.3,0.1

Type RM Length L Ch R = 1 ,15625   ,120,120,120
BEGIN DESCRIPTION:
MACK CREEK 28.0
END DESCRIPTION:
XS GIS Cut Line= 3
      3730149.21      10602389.3      3729917.44     10602837.23
       3729644.3     10602912.66
#Sta/Elev= 30
  4754.9  254.09  4915.1     254  4947.3  254.42  4956.8  252.05  4969.8  244.65
    4979  241.68  4984.6  236.39    4991  234.38  4998.1  233.67  5000.9  233.17
  5004.1  233.67  5014.9  235.15  5028.9  242.09    5051  243.71  5067.5  242.64
  5089.7  248.29  5099.3  248.33  5127.5  247.86  5139.6  249.77  5147.6  249.05
  5178.2  251.64  5183.9  253.35  5223.2  257.52    5340  262.44  5365.1  266.24
  5371.1  274.32  5381.5   277.2  5481.9  291.77  5512.8  295.18  5542.6     296
#Mann= 9 ,-1 , 0
  4754.9     .05       0  4915.1     .16       0    4991     .08       0
  4998.1     .07       0  5004.1     .08       0  5099.3     .05       0
  5147.6     .16       0  5223.2     .05       0  5481.9     .16       0
Bank Sta=4979,5028.9
XS Rating Curve= 0 ,0
Exp/Cntr=0.3,0.1

Type RM Length L Ch R = 1 ,15505   ,411,411,411
BEGIN DESCRIPTION:
Mapping XS 1160fd7f
END DESCRIPTION:
XS GIS Cut Line= 2
      3730115.38      10602397.1      3729719.56     10602704.39
#Sta/Elev= 30
  4793.3  253.66    4914  252.95  4935.2  250.22  4941.6  246.31  4949.7  244.61
    4985  240.89  4991.4  238.81  4999.5  233.49  5002.8  233.11  5005.6  232.61
  5008.8  233.11    5014  233.49  5020.3  239.16  5034.8  241.92  5055.6  239.99
  5091.8  243.85  5113.5  254.19  5134.4  258.08  5142.4  262.46  5169.7  266.04
  5177.8  269.48  5184.1  268.83  5192.3  274.97  5198.6  271.76  5205.7  277.74
  5213.1  281.42  5219.4  280.46  5227.6   284.3  5248.4  287.13  5294.4  290.45
#Mann= 4 ,-1 , 0
  4793.3     .05       0    4914     .13       0  5002.8     .07       0
  5008.8     .13       0
Bank Sta=4991.4,5020.3
XS Rating Curve= 0 ,0
Exp/Cntr=0.3,0.1

Type RM Length L Ch R = 1 ,15094   ,606,606,606
BEGIN DESCRIPTION:
MACK CREEK 27.0
END DESCRIPTION:
XS GIS Cut Line= 3
      3730302.88     10602225.26       3729831.5     10602105.46
      3729706.43     10602226.33
#Sta/Elev= 30
  4663.6  260.17  4739.2  254.92  4744.7  253.72  4749.9  250.74  4770.2   249.6
  4780.5  244.34  4785.7  244.64  4790.8  242.69  4867.5  239.02  4935.2  238.91
  4949.4  240.71  4976.5  238.31  4985.2  232.81  4994.2  231.59  4996.9  231.09
  5000.2  231.59  5015.8  236.34  5017.8  236.93  5026.1   243.9  5031.3   249.8
  5038.4  251.32    5108  251.85  5190.1  250.06  5218.4  251.84  5225.3  253.76
  5246.7  253.96  5253.6  255.86  5310.2  260.24  5317.4  259.43  5323.9  260.97
#Mann= 4 ,-1 , 0
  4663.6     .05       0  4994.2     .03       0  5000.2     .05       0
  5015.8     .16       0
Bank Sta=4976.5,5017.8
XS Rating Curve= 0 ,0
Exp/Cntr=0.3,0.1

Type RM Length L Ch R = 1 ,14488   ,669,669,669
BEGIN DESCRIPTION:
MACK CREEK 26.0
END DESCRIPTION:
XS GIS Cut Line= 3
      3730254.08      10601576.1      3729833.09     10602040.49
      3729676.99     10602199.31
#Sta/Elev= 30
  4790.1  284.76  4852.6  284.24  4860.1  283.85  4866.8   281.4  4888.4  280.35
  4902.6  270.02  4909.4  259.17  4916.8   253.8  4944.5  244.46    4952  240.72
  4966.2  239.25  4972.9  234.64  4980.4  232.03  4994.5  229.29  5005.7  228.93
  5008.5  228.43  5011.7  228.93  5022.9  239.86  5029.7  242.02  5037.1  247.35
  5100.6  250.03  5291.9  249.98    5327  248.78  5348.7   250.1  5404.8  249.41
  5454.5  250.65  5482.8   249.2  5518.1  249.38  5560.6  251.53  5639.6  258.71
#Mann= 3 ,-1 , 0
  4790.1     .16       0  5005.7     .07       0  5011.7     .16       0
Bank Sta=4966.2,5022.9
XS Rating Curve= 0 ,0
Exp/Cntr=0.3,0.1

Type RM Length L Ch R = 1 ,13819   ,232,232,232
BEGIN DESCRIPTION:
MACK CREEK 25.0
END DESCRIPTION:
XS GIS Cut Line= 3
      3729784.62     10601339.85      3729630.98     10601772.12
      3729566.04     10602146.16
#Sta/Elev= 30
  4457.3  267.52  4485.7  265.27  4510.7  261.06  4572.9  257.51  4578.2  255.02
  4627.5  251.14  4670.8  245.17  4736.8  243.83    4776  246.28  4807.9  245.32
  4814.4  241.24  4815.8  242.27  4819.7  245.13  4850.6  243.97  4870.8  245.34
  4882.2  238.25  4916.1  238.47    4975  232.61  4992.3  225.76  4995.1  225.26
  4998.3  225.76  5016.2  228.25  5025.7  234.52  5056.2  236.15  5065.8  240.53
  5076.5     241  5086.6  248.37  5096.8  249.69  5198.7  254.44  5295.7   259.5
#Mann= 6 ,-1 , 0
  4457.3     .16       0  4736.8     .12       0  4815.8     .16       0
  4992.3     .07       0  4998.3     .16       0  5198.7     .12       0
Bank Sta=4975,5025.7
XS Rating Curve= 0 ,0
Exp/Cntr=0.3,0.1

Type RM Length L Ch R = 1 ,13587   ,179,179,179
BEGIN DESCRIPTION:
Mapping XS f3205d51
END DESCRIPTION:
XS GIS Cut Line= 3
      3729681.31     10601386.88      3729519.84     10601645.58
      3729275.08      10601902.5
#Sta/Elev= 30
  4635.6  260.33  4640.5  260.33  4646.8  256.71  4652.7  257.52  4704.6  247.99
    4799  244.42  4804.9  239.54  4835.6  244.56  4850.9  243.47  4856.8  241.01
  4872.3  241.19    4878  239.41    4887  241.44  4899.3  238.74  4908.7  239.94
  4965.1  236.02  4972.4  232.83  4986.5  231.96  4997.7  224.41  5000.4  223.91
  5003.7  224.41  5014.9  225.04  5021.8  230.09  5050.1  239.91  5057.3  239.29
  5078.4  243.18  5085.3  247.99  5099.4  250.77  5219.9  256.47  5295.4  257.27
#Mann= 4 ,-1 , 0
  4635.6     .12       0  4872.3     .16       0  4997.7     .07       0
  5003.7     .16       0
Bank Sta=4986.5,5021.8
XS Rating Curve= 0 ,0
Exp/Cntr=0.3,0.1

Type RM Length L Ch R = 1 ,13408   ,144,144,144
BEGIN DESCRIPTION:
MACK CREEK 24.0
END DESCRIPTION:
XS GIS Cut Line= 2
      3729602.31     10601290.38      3729121.75     10601856.66
#Sta/Elev= 30
  4685.9  280.29  4707.2  279.27  4751.2   272.7  4787.3  248.26    4803  245.39
  4829.9  242.02  4857.5  244.01  4886.1  235.88  4957.5  235.51  4978.4  230.51
  4986.1  227.88  4989.6  223.88  4992.4  223.38  4995.6  223.88  5021.2  230.37
  5042.1  234.16  5049.8  245.63  5070.6  246.78  5191.5  251.24  5248.6  247.26
  5255.2  241.01  5269.5  249.35    5276  242.61  5290.3  244.13    5298   241.9
  5304.6  250.53  5326.6  251.04  5333.2  253.63  5340.9  252.08  5428.6  267.67
#Mann= 5 ,-1 , 0
  4685.9     .16       0  4707.2     .12       0    4803     .16       0
  4989.6     .07       0  4995.6     .16       0
Bank Sta=4978.4,5021.2
XS Rating Curve= 0 ,0
Exp/Cntr=0.3,0.1

Type RM Length L Ch R = 1 ,13264   ,181,181,181
BEGIN DESCRIPTION:
Mapping XS f035166f
END DESCRIPTION:
XS GIS Cut Line= 4
      3729578.87     10601244.54      3729334.08     10601395.58
      3729224.71     10601499.75      3728969.78     10601775.48
#Sta/Elev= 30
  4672.1   281.3  4748.6  274.87    4764  270.13  4791.1  253.77  4812.4  248.15
  4980.2  229.64  4998.6  223.41  5001.3  222.91  5004.6  223.41  5022.6  229.51
  5029.9  230.56  5036.8  239.64    5044  241.97  5114.6  238.51  5128.7  241.02
  5142.9  239.09  5150.3  233.32  5178.6  240.24  5206.7  240.81  5220.6   247.6
    5228   244.9  5234.8  249.81  5242.1  246.41  5248.9  250.31  5341.4  253.63
  5447.4  262.08  5454.2  266.91  5475.7  265.64  5482.5  270.27  5486.3  267.49
#Mann= 3 ,-1 , 0
  4672.1     .16       0  4998.6     .07       0  5004.6     .16       0
Bank Sta=4980.2,5022.6
XS Rating Curve= 0 ,0
Exp/Cntr=0.3,0.1
