HEC-RAS study TOWN CREEK.prj: TOWN CREEK Base Level Engineering

--- TOWN CREEK.g01 (geometry) --- (continued)

Type RM Length L Ch R = 1 ,48896   ,605,605,605
BEGIN DESCRIPTION:
TOWN CREEK 66.0
END DESCRIPTION:
XS GIS Cut Line= 3
      3731299.61     10620610.16      3731299.61     10621210.19
      3731149.62     10621610.17
#Sta/Elev= 30
  4383.3  283.21  4423.3  281.95  4543.3  270.38  4557.8 267.969  4603.3  262.91
  4633.3  261.03  4753.3  262.57  4793.3  261.61  4843.3   263.7  4903.3  263.57
  4953.3  265.22    4986  263.67  4993.1  255.91    4997  254.82  4999.8  254.32
    5003  254.82  5004.7  254.82  5015.4  260.57  5023.4  262.39  5028.7  265.64
  5047.4  264.33  5114.2  263.78  5139.1  267.03  5169.3     268  5224.5  273.61
  5229.9  272.79  5279.7  277.11    5285  276.63  5365.1  285.34  5410.5  287.29
#Mann= 5 ,-1 , 0
  4383.3     .05       0  4557.8     .16       0    4997     .07       0
    5003     .16       0  5047.4     .05       0
Bank Sta=4986,5028.7
XS Rating Curve= 0 ,0
Exp/Cntr=0.3,0.1

Type RM Length L Ch R = 1 ,48291   ,539,539,539
BEGIN DESCRIPTION:
TOWN CREEK 65.0
END DESCRIPTION:
XS GIS Cut Line= 3
      3730949.61      10620560.2      3730849.61     10621110.19
      3730799.61     10621660.22
#Sta/Elev= 30
  4461.8  289.78  4546.9  287.93  4583.8  284.01  4653.6  274.26  4658.7  274.77
  4685.4  271.45  4817.5  259.38    4848  259.06    4867262.7308  4940.8  262.39
    4970   264.2  4978.1263.6707  4980.1  263.54    4989  257.35  4994.1  257.15
    4997  253.85  4999.8  253.35    5003  253.85  5010.6  253.85  5018.3  263.06
  5050.9  264.11  5076.6262.8628  5121.2  261.53  5261.8  261.46  5291.9  264.19
    5302  266.38    5312  266.34  5372.2  272.35  5462.6  282.81  5573.1  297.96
#Mann= 6 ,-1 , 0
  4461.8     .05       0    4867     .12       0  4978.1     .16       0
    4997     .07       0    5003     .16       0  5076.6     .05       0
Bank Sta=4980.1,5018.3
XS Rating Curve= 0 ,0
Exp/Cntr=0.3,0.1

Type RM Length L Ch R = 1 ,47752   ,579,579,579
BEGIN DESCRIPTION:
TOWN CREEK 64.0
END DESCRIPTION:
XS GIS Cut Line= 3
       3730899.6      10620610.2      3730399.61     10621010.19
      3730049.62     10621260.18
#Sta/Elev= 30
  4355.3  288.79  4412.1  286.23  4476.1  279.15    4505   273.9  4622.4266.2069
  4725.9  263.24  4732.3  264.46  4739.5  262.33  4796.3  260.55  4817.1  262.23
    4982  263.12  4988.4   253.6  4995.6   255.1    4997  253.47  4999.8  252.97
    5003  253.47  5009.1  255.75  5017.7   255.8  5023.9  260.78  5032.5  259.86
  5053.4  262.77  5109.9  260.02  5154.1  261.42  5160.3   259.4  5181.2  260.97
  5240.2  271.38  5302.8  285.92  5347.1  291.52    5368  296.14  5425.7  302.62
#Mann= 4 ,-1 , 0
  4355.3     .05       0  4622.4     .12       0    4997     .07       0
    5003     .12       0
Bank Sta=4982,5023.9
XS Rating Curve= 0 ,0
Exp/Cntr=0.3,0.1

Type RM Length L Ch R = 1 ,47173   ,541,541,541
BEGIN DESCRIPTION:
TOWN CREEK 63.0
END DESCRIPTION:
XS GIS Cut Line= 3
      3730200.63     10619730.47      3730214.52     10620542.95
      3729944.74     10621165.52
#Sta/Elev= 30
  4090.6  310.06  4094.9309.9141  4380.4  306.09  4460.4  297.79  4580.4  272.38
  4640.4  262.17  4660.4  260.25  4740.4  261.08  4750.4  253.24  4760.4  252.56
  4790.4   260.9  4820.4  260.52  4830.4  258.65  4840.4  260.77    4922  259.05
  4974.7  262.29  4980.2  259.62  4987.4  253.07    4997  252.56  4999.8  252.06
    5003  252.56  5027.1  261.36    5140  262.88  5194.4  268.52  5377.5  280.41
  5412.4  286.66  5476.9  292.47  5488.7   295.7  5499.6  295.24  5581.7   301.9
#Mann= 4 ,-1 , 0
  4090.6     .05       0  4094.9     .12       0    4997     .07       0
    5003     .12       0
Bank Sta=4974.7,5027.1
XS Rating Curve= 0 ,0
Exp/Cntr=0.3,0.1

Type RM Length L Ch R = 1 ,46632   ,560,560,560
BEGIN DESCRIPTION:
TOWN CREEK 62.0
END DESCRIPTION:
XS GIS Cut Line= 3
      3729599.62      10619960.2      3729799.61     10620360.19
      3729799.61     10621160.19
#Sta/Elev= 30
  4517.5  310.85  4550.2307.5421  4637.7   298.8  4643.3  299.31    4660   296.5
  4665.6  297.58  4710.3  290.98  4718.7  288.58  4732.7  287.08  4741.1  283.39
  4755.1  281.38  4794.2  269.22  4808.2  263.11  4830.5  258.87  4852.9  257.74
  4967.2  260.96    4997  251.76  4999.8  251.26    5003  251.76  5024.7  253.12
  5034.7  260.93  5194.7  260.39  5214.7  258.91  5354.7  259.15  5404.7  260.98
  5444.7  263.63  5504.7  270.47  5644.7  292.47  5684.7  297.79  5764.7  305.14
#Mann= 4 ,-1 , 0
  4517.5     .05       0  4550.2     .12       0    4997     .07       0
    5003     .12       0
Bank Sta=4967.2,5034.7
XS Rating Curve= 0 ,0
Exp/Cntr=0.3,0.1

Type RM Length L Ch R = 1 ,46072   ,488,488,488
BEGIN DESCRIPTION:
TOWN CREEK 61.0
END DESCRIPTION:
XS GIS Cut Line= 3
      3729449.63     10619910.15      3729299.61     10620310.19
      3729649.63     10621110.23
#Sta/Elev= 30
  4583.3  309.87  4623.4  308.65  4628.7  306.39  4654.7304.6851  4799.6  291.41
  4871.7  287.72  4940.2  278.86  4965.2  272.12  4970.5  273.11  4989.2  259.24
  4995.4  251.08    4997  250.83  4999.8  250.33    5003  250.83  5013.3  250.85
  5022.6  255.14  5032.4  260.15  5113.5259.0296    5241258.2082  5349.9257.8227
    5403257.0246  5534.5  256.27  5567.6257.9578    5589  258.42  5665.5  265.43
  5736.9274.7421  5785.5  283.93  5807.4  285.01  5817.1  287.86  5883.8  296.63
#Mann= 11 ,-1 , 0
  4583.3     .05       0  4654.7     .12       0    4997     .07       0
    5003     .12       0  5022.6     .16       0  5113.5     .12       0
    5241     .16       0  5349.9     .12       0    5403     .16       0
  5567.6     .12       0  5736.9     .05       0
Bank Sta=4989.2,5032.4
XS Rating Curve= 0 ,0
Exp/Cntr=0.3,0.1

Type RM Length L Ch R = 1 ,45584   ,406,406,406
BEGIN DESCRIPTION:
TOWN CREEK 60.0
END DESCRIPTION:
XS GIS Cut Line= 3
      3729054.63     10619747.62      3728776.86     10620676.43
      3728378.06     10621265.96
#Sta/Elev= 30
  4323.6   281.6  4426.9  278.37  4524.6     271  4536.7   268.8  4597.7  267.96
  4629.4265.7263  4681.2  258.04  4707.4  256.89  4921.7   257.8  4973.4  259.65
  4982.7  255.76  4987.9  250.29    4997  249.84  4999.8  249.34    5003  249.84
    5021  259.24    5036     260  5077.8  256.98  5150.9  255.55  5387.2  258.65
  5474.1   263.3  5563.9  272.02    5582  273.65    5588  276.09  5596.9  275.38
  5638.9  280.72  5725.8  288.44  5782.7  288.54  5920.5  283.38  6004.8  284.04
#Mann= 5 ,-1 , 0
  4323.6     .05       0  4629.4     .12       0    4997     .07       0
    5003     .12       0  5563.9     .05       0
Bank Sta=4973.4,5021
XS Rating Curve= 0 ,0
Exp/Cntr=0.3,0.1

Type RM Length L Ch R = 1 ,45178   ,545,545,545
BEGIN DESCRIPTION:
Mapping XS 86662fb9
END DESCRIPTION:
XS GIS Cut Line= 3
      3728768.77     10619491.32      3728565.63     10620199.69
      3728201.05     10621137.18
#Sta/Elev= 30
  4124.8  299.98  4284.9  284.53  4337.5 281.834  4414.9  278.74  4560.5   280.6
  4609.4  278.84    4675  272.36  4687.3  268.08  4706.2  266.57  4721.1  259.88
  4737.4  256.49  4915.1  258.85  4926.6  255.24  4958.8  255.63  4969.5  254.39
  4980.3  249.46    4997  249.33  4999.8  248.83    5003  249.33  5004.8  252.51
  5023.2  256.01  5029.3  252.34  5034.7  259.31  5143.5  255.96  5216.3  257.12
  5391.1  267.63  5540.4 279.948  5777.3  292.94  5856.3  295.25  5867.6  297.14
#Mann= 5 ,-1 , 0
  4124.8     .05       0  4337.5     .12       0    4997     .07       0
    5003     .12       0  5540.4     .05       0
Bank Sta=4915.1,5034.7
XS Rating Curve= 0 ,0
Exp/Cntr=0.3,0.1

Type RM Length L Ch R = 1 ,44633   ,642,642,642
BEGIN DESCRIPTION:
Mapping XS 3523af8f
END DESCRIPTION:
XS GIS Cut Line= 3
        3728649.     10619303.83      3728336.47     10619533.02
      3728091.68     10620730.91
#Sta/Elev= 30
  4276.7  295.28  4380.9  281.85  4431.1  271.89  4481.2  264.77  4516.7  262.39
  4573.6  254.69  4725.6  254.43  4972.9  258.56    4988  253.64    4997  248.49
  4999.8  247.99    5003  248.49  5018.3  248.49  5028.8  254.15    5039  256.95
  5151.3  254.73  5225.4  259.26  5321.3  260.42  5472.7  268.12  5498.3  267.85
  5518.1  269.06  5559.6  276.28  5573.7  282.16  5610.6  285.65  5624.2  288.95
  5668.9 292.134  5720.1  295.94  5733.1   299.6  5826.2  303.85  5886.9   304.2
#Mann= 4 ,-1 , 0
  4276.7     .12       0    4997     .07       0    5003     .12       0
  5668.9     .05       0
Bank Sta=4972.9,5039
XS Rating Curve= 0 ,0
Exp/Cntr=0.3,0.1

Type RM Length L Ch R = 1 ,43991   ,610,610,610
BEGIN DESCRIPTION:
Mapping XS 619b8410
END DESCRIPTION:
XS GIS Cut Line= 3
      3728668.11      10619082.8      3728016.49     10619300.01
      3728022.28     10620571.52
#Sta/Elev= 30
  4430.5  299.32  4460.5  292.47  4544.9  280.87  4576.5   274.6  4618.7  268.92
  4695.2262.3287  4720.7  257.72  4766.2  253.71  4866.2 253.972    4979  257.53
  4987.6  249.31    4997  247.19  4999.8  246.69    5003  247.19  5010.6  247.39
  5029.8  256.46  5050.8  255.31  5068.6  259.17  5113.1   263.7  5177.6  264.02
  5257.6  262.43  5407.6  255.56  5487.6  255.93  5627.6  264.39  5697.6  266.11
  5777.6  272.05  5927.6  276.76  6017.6  284.25  6100.7287.4532  6388.9  300.73
#Mann= 6 ,-1 , 0
  4430.5     .12       0  4695.2     .16       0  4866.2     .12       0
    4997     .07       0    5003     .12       0  6100.7     .05       0
Bank Sta=4979,5029.8
XS Rating Curve= 0 ,0
Exp/Cntr=0.3,0.1

Type RM Length L Ch R = 1 ,43381   ,694,694,694
BEGIN DESCRIPTION:
TOWN CREEK 59.0
END DESCRIPTION:
XS GIS Cut Line= 3
      3728581.27     10618100.93      3727839.81      10619068.3
      3727929.54     10620556.06
#Sta/Elev= 30
    4231  297.48  4274.4298.6776  4374.2  289.14  4394.9284.8041  4473.9  273.55
  4602.7   261.2    4852  256.67  4866.5  257.91  4901.8  255.96  4973.4  256.73
    4987  247.12    4997  246.46  4999.8  245.96    5003  246.46    5016  252.52
  5036.9  256.45  5165.6  254.68  5250.8   256.7  5394.1  255.75  5414.9  254.22
  5521.9  257.11  5652.1  252.03  5832.4  251.88  6027.8  258.64  6042.8  257.68
  6323.3  265.02  6522.4  283.53  6646.7  293.09  6864.3  301.09  6940.3  302.09
#Mann= 6 ,-1 , 0
    4231     .12       0  4274.4     .16       0  4394.9     .12       0
    4997     .07       0    5003     .12       0  6646.7     .05       0
Bank Sta=4973.4,5036.9
XS Rating Curve= 0 ,0
Exp/Cntr=0.3,0.1

Type RM Length L Ch R = 1 ,42687   ,236,236,236
BEGIN DESCRIPTION:
TOWN CREEK 58.0
END DESCRIPTION:
XS GIS Cut Line= 3
       3726914.6     10618283.03      3727570.84     10618678.86
      3727878.13     10620710.07
#Sta/Elev= 30
  3971.5  300.76  3973.6  297.74    3989  297.38  4016.3  300.58  4117.5  285.36
  4289.9267.2988  4346.5259.4637  4381.3  254.06  4549.4  254.06    4608  256.61
  4635.6  253.16  4686.7253.5431  4820.1  251.91  4903.1254.2127  4904.3254.3204
  4960.1  255.38    4997  245.28  4999.8  244.78    5003  245.28  5022.4  245.28
    5034  253.53  5437.1  251.25  5710.1  265.91  5791.1  265.92  5861.9  270.08
  6104.9  270.25  6320.4282.9837  6418.1  286.37  6571.5  296.41  6792.2  299.48
#Mann= 10 ,-1 , 0
  3971.5     .05       0  4289.9     .16       0  4346.5     .05       0
  4549.4     .16       0  4686.7     .12       0  4903.1     .16       0
  4904.3     .12       0    4997     .07       0    5003     .12       0
  6320.4     .05       0
Bank Sta=4960.1,5034
XS Rating Curve= 0 ,0
Exp/Cntr=0.3,0.1

Type RM Length L Ch R = 1 ,42451   ,955,955,955
BEGIN DESCRIPTION:
TOWN CREEK 57.0
END DESCRIPTION:
XS GIS Cut Line= 3
      3726826.04     10618454.89      3727367.72     10618835.11
      3727643.37     10620176.99
#Sta/Elev= 30
    4233  301.74  4282.9  301.05  4318.7  307.01  4339.6  299.96  4360.5  302.76
    4411  297.24  4440.7  288.32  4461.6   286.3  4476.4  280.29  4512.1  274.64
  4541.8  264.79  4613.2  257.54  4619.3  254.36  4777.2250.7324  4892.9  251.45
  4924.1254.5132  4933.7254.4255  4971.4  253.91  4977.7  247.99  4982.8  253.83
    4997  245.11  4999.8  244.61    5003  245.11  5012.3  245.17  5042.9  254.78
  5330.2  250.94  5728.1  266.29  6020.1  281.65  6120.8  283.77  6264.7  280.78
#Mann= 6 ,-1 , 0
    4233     .05       0  4777.2     .12       0  4924.1     .16       0
  4933.7     .12       0    4997     .07       0    5003     .12       0
Bank Sta=4982.8,5042.9
XS Rating Curve= 0 ,0
Exp/Cntr=0.3,0.1

Type RM Length L Ch R = 1 ,41496   ,556,556,556
BEGIN DESCRIPTION:
TOWN CREEK 56.0
END DESCRIPTION:
XS GIS Cut Line= 3
      3726399.57     10619010.17      3726749.61     10619210.19
      3727449.63      10619560.2
#Sta/Elev= 30
  4598.1  305.29    4602305.3076  4643.5  302.72  4665.1  299.48  4701.8  292.08
  4708.3  289.34  4729.9  286.66  4736.4  283.83  4751.5  281.76  4788.9   272.3
  4897.6  253.83  4971.7  253.45  4978.2  246.72  4987.6  244.11    4997  243.96
  4999.8  243.46    5003  243.96  5009.6  246.71  5015.2  244.18    5032  253.07
  5037.6  249.86    5046  252.85  5054.4  253.11  5188.5  250.49  5342.2250.8161
  5519.1248.7425  5551.9  247.82  5613.4  255.38  5730.8     267  5783.9  268.08
#Mann= 6 ,-1 , 0
  4598.1     .05       0    4602     .12       0    4997     .07       0
    5003     .12       0  5342.2     .16       0  5519.1     .12       0
Bank Sta=4971.7,5032
XS Rating Curve= 0 ,0
Exp/Cntr=0.3,0.1

Type RM Length L Ch R = 1 ,40940   ,636,636,636
BEGIN DESCRIPTION:
TOWN CREEK 55.0
END DESCRIPTION:
XS GIS Cut Line= 3
      3726199.58     10619210.18      3726999.61     10619560.19
      3727349.65     10619760.21
#Sta/Elev= 30
  4097.8  295.24  4174.2  282.43  4182.4  277.07  4187.9  279.49  4196.1  273.59
  4217.9  277.99  4250.6  276.52  4409.3  253.63  4454.9252.0907  4645.8 251.757
  4787.4  253.19  4796.4  247.05  4805.4  245.14  4810.8  249.24  4828.8  244.09
  4834.2  252.59  4840.1  248.18  4857.6  247.79  4863.1  253.18  4984.7  251.35
    4997  242.55  4999.8  242.05    5003  242.55  5022.2  244.23  5028.6  251.96
  5059.6  251.81  5086.9  247.65  5118.6  248.47  5307.2  279.16  5374.2  286.04
#Mann= 5 ,-1 , 0
  4097.8     .12       0  4454.9     .16       0  4645.8     .12       0
    4997     .07       0    5003     .12       0
Bank Sta=4984.7,5028.6
XS Rating Curve= 0 ,0
Exp/Cntr=0.3,0.1

Type RM Length L Ch R = 1 ,40304   ,530,530,530
BEGIN DESCRIPTION:
TOWN CREEK 54.0
END DESCRIPTION:
XS GIS Cut Line= 3
      3726399.63     10619960.19      3726799.61     10619910.19
       3727299.6     10620110.19
#Sta/Elev= 30
  4573.2  287.06  4603.4  285.16    4674   275.7    4684  275.46  4694.8273.0157
  4764.7  265.26  4784.8  261.11  4825.1  256.76  4875.5  247.39  4885.6  247.18
  4915.8  250.84  4966.2  251.79    4979  250.05  4985.7  245.72  4991.1  249.49
    4997  242.37  4999.8  241.87    5003  242.37  5008.6  244.47  5015.3  250.99
  5020.7  246.73  5030.1  251.35  5116.3  249.65  5159.4  252.77  5314.2   269.7
  5320.9  272.28  5353.3  277.51  5368.1  278.33  5392.3   283.9  5514.8  298.99
#Mann= 4 ,-1 , 0
  4573.2     .16       0  4694.8     .12       0    4997     .07       0
    5003     .12       0
Bank Sta=4991.1,5015.3
XS Rating Curve= 0 ,0
Exp/Cntr=0.3,0.1

Type RM Length L Ch R = 1 ,39774   ,619,619,619
BEGIN DESCRIPTION:
TOWN CREEK 53.0
END DESCRIPTION:
XS GIS Cut Line= 3
      3726399.62     10620210.19      3726849.61     10620310.19
      3727249.63     10620260.19
#Sta/Elev= 30
  4536.9  286.38  4561.2  285.49  4567.6   282.8  4588.1  279.03  4628.5273.6953
  4696.9  262.66  4813.5  250.39  4864.7  248.06  4895.4  250.48  4973.5  250.69
  4978.7  249.74  4987.6  241.93    4997  240.83  4999.8  240.33    5003  240.83
    5018  240.83  5028.1  243.07  5035.7  250.16  5040.7  245.56  5048.3  244.29
  5058.3  250.46  5068.4  251.43    5149  251.98  5189.3  260.88  5196.9  264.46
  5229.7  269.81    5270  278.93  5277.5  283.33  5310.3  288.13    5401  294.69
#Mann= 4 ,-1 , 0
  4536.9     .16       0  4628.5     .12       0    4997     .07       0
    5003     .12       0
Bank Sta=4973.5,5035.7
XS Rating Curve= 0 ,0
Exp/Cntr=0.3,0.1

Type RM Length L Ch R = 1 ,39155   ,541,541,541
BEGIN DESCRIPTION:
TOWN CREEK 52.0
END DESCRIPTION:
XS GIS Cut Line= 3
      3726299.63     10620310.21      3726699.61     10620810.19
      3727049.61     10621010.19
#Sta/Elev= 30
  4345.9  290.35  4383.3288.4495  4460.3  278.59  4516.4  267.09  4580.4  257.49
  4687.6  248.61  4730.1  246.89  4836.5  248.72  4865.3  250.48  4879.7  249.38
  4964.6  250.86    4979  248.04    4983  242.56    4997  240.42  4999.8  239.92
    5003  240.42  5015.7  240.42  5021.5  245.81  5031.5  249.55  5043.8  250.95
  5058.9  250.33  5065.3251.9827  5161.1  274.63  5170.5  275.48  5182.7  278.93
  5192.8  278.67    5205  283.04  5263.3  290.15  5285.2  290.81  5389.3  296.34
#Mann= 6 ,-1 , 0
  4345.9     .05       0  4383.3     .12       0    4997     .07       0
    5003     .12       0  5065.3     .16       0  5285.2     .05       0
Bank Sta=4964.6,5031.5
XS Rating Curve= 0 ,0
Exp/Cntr=0.3,0.1

Type RM Length L Ch R = 1 ,38614   ,621,621,621
BEGIN DESCRIPTION:
TOWN CREEK 51.0
END DESCRIPTION:
XS GIS Cut Line= 3
      3726149.61     10620410.17      3726199.61     10620860.19
      3726499.64     10621160.22
#Sta/Elev= 30
  4546.5  286.96  4631.5280.7942  4677.3  275.79  4687.4  272.19  4717.6  267.55
  4727.6  264.85    4788  255.35  4838.3  249.03  4868.5  248.11  4878.6  246.66
  4923.2246.8346  4979.2  248.98  4989.2  245.94    4997  239.37  4999.8  238.87
    5003  239.37  5013.4  239.77  5027.6  248.63  5041.7  249.94  5098.3  248.83
  5126.6  249.81  5176.1  259.46  5225.6  266.28  5239.7  270.43  5253.8  272.09
  5282.1  278.12  5324.6  281.63    5353 281.463  5409.4  281.98  5423.6  282.18
#Mann= 7 ,-1 , 0
  4546.5     .05       0  4631.5     .07       0  4923.2     .12       0
    4997     .07       0    5003     .12       0    5353     .05       0
  5409.4     .12       0
Bank Sta=4979.2,5027.6
XS Rating Curve= 0 ,0
Exp/Cntr=0.3,0.1

Type RM Length L Ch R = 1 ,37993   ,388,388,388
BEGIN DESCRIPTION:
TOWN CREEK 50.0
END DESCRIPTION:
XS GIS Cut Line= 3
      3725576.05     10619783.03      3725622.92     10620944.48
       3726034.4     10621553.88
#Sta/Elev= 30
  3732.8  295.69    3830  300.37    4064 300.608    4186298.6743  4423.5 295.183
  4510.6  290.56  4550.6  286.08  4576.8280.8031  4687.4  255.58  4692.4  257.87
  4700.7  254.34  4718.5251.3651  4740.8  247.61  4816.8 245.714  4933.1   249.9
  4962.4  249.81    4984  247.14  4990.1  238.44    4997  238.44  4999.8  237.94
    5003  238.44  5011.1  238.52    5026  248.42  5214.8  245.43  5385.7   265.3
  5436.7  263.91  5451.6  257.99  5472.6  257.56  5559.5  274.06  5630.5  282.93
#Mann= 9 ,-1 , 0
  3732.8     .05       0    4064     .12       0    4186     .05       0
  4423.5     .07       0  4576.8     .12       0  4718.5     .07       0
  4816.8     .12       0    4997     .07       0    5003     .12       0
Bank Sta=4984,5026
XS Rating Curve= 0 ,0
Exp/Cntr=0.3,0.1

Type RM Length L Ch R = 1 ,37605   ,673,673,673
BEGIN DESCRIPTION:
TOWN CREEK 49.0
END DESCRIPTION:
XS GIS Cut Line= 3
      3724424.97     10620611.12      3725372.92     10621230.94
      3725800.02     10621684.08
#Sta/Elev= 30
  3804.4  296.19  4037.2290.5383  4052.1   289.6  4067.2  292.22  4103.4  293.65
  4196.9  292.02  4240.1  293.34  4335.6  290.45  4409.9284.0368  4435.2  278.42
  4450.3  280.22  4505.5271.5534  4631.2  258.57  4682.1  257.51  4724.7  253.54
  4745.8  254.39  4911.7  245.89  4969.5   247.7  4983.6  244.27    4997  238.08
  4999.8  237.58    5003  238.08  5018.8  241.76  5026.1  247.66  5125.2  245.84
    5196  250.08  5287.9  262.22  5351.4  267.69  5557.3  296.78  5559.7  296.78
#Mann= 7 ,-1 , 0
  3804.4     .16       0  4037.2     .05       0  4409.9     .07       0
  4505.5     .12       0    4997     .07       0    5003     .12       0
  5557.3     .05       0
Bank Sta=4969.5,5026.1
XS Rating Curve= 0 ,0
Exp/Cntr=0.3,0.1

Type RM Length L Ch R = 1 ,36932   ,549,549,549
BEGIN DESCRIPTION:
TOWN CREEK 48.0
END DESCRIPTION:
XS GIS Cut Line= 3
      3724649.59     10621560.18      3724999.61     10621760.19
      3725749.61     10621810.19
#Sta/Elev= 30
  4564.8  280.89  4695.4278.8186  4719.5 277.549  4777.2  271.48    4793  267.83
  4798.8  268.55  4806.7  265.57  4820.4  265.47  4873.6  257.75  4879.4  259.13
  4892.8255.4245  4938.4  251.07  4954.3  245.58    4978  247.13    4988  239.18
    4997  237.13  4999.8  236.63    5003  237.13    5018  237.88  5028.1  247.96
  5038.1  249.08  5118.3  243.93  5208.5   245.3  5278.6  249.23  5288.6  251.61
  5318.7  252.69  5398.9  261.71  5589.3  287.48  5649.4  298.28  5719.6  305.47
#Mann= 6 ,-1 , 0
  4564.8     .07       0  4695.4     .05       0  4719.5     .07       0
  4892.8     .12       0    4997     .07       0    5003     .12       0
Bank Sta=4978,5028.1
XS Rating Curve= 0 ,0
Exp/Cntr=0.3,0.1

Type RM Length L Ch R = 1 ,36383   ,512,512,512
BEGIN DESCRIPTION:
TOWN CREEK 47.0
END DESCRIPTION:
XS GIS Cut Line= 3
      3724699.63     10621810.21      3725099.61     10622260.19
      3725499.57     10622510.17
#Sta/Elev= 30
  4396.9  269.12  4510.2  260.47  4687.5   254.6  4715.9  250.85  4722.6  247.96
  4730.1  248.13  4736.8  246.17  4744.3  248.39    4751  245.12  4771.9   247.2
  4806.8247.8162  4864.7  248.14  4871.4  246.11  4892.3  248.13  4956.7  248.22
  4985.1  244.27  4991.8  236.14    4997  236.14  4999.8  235.64    5003  236.14
  5012.5  242.03  5027.8  247.09  5034.3  244.59  5064.4  243.79  5187.6  256.29
  5378.4279.6391  5399.3  281.49  5411.7  285.17  5452.5290.9575  5470.6  293.41
#Mann= 6 ,-1 , 0
  4396.9     .07       0  4806.8     .12       0    4997     .07       0
    5003     .12       0  5378.4     .07       0  5452.5     .05       0
Bank Sta=4956.7,5027.8
XS Rating Curve= 0 ,0
Exp/Cntr=0.3,0.1

Type RM Length L Ch R = 1 ,35871   ,655,655,655
BEGIN DESCRIPTION:
Mapping XS 52503482
END DESCRIPTION:
XS GIS Cut Line= 3
      3723820.87     10621673.67      3724716.67     10622428.86
      3725221.89     10622829.91
#Sta/Elev= 30
  3725.1  275.77  3792.5  273.65  3828.1   275.8  3835.3  272.26  3841.9  274.08
  3849.6  270.87  3856.2  274.26  3878.2  270.06  3884.8  272.61  3927.7  272.47
  3934.2  275.39    3942  271.21  3972.7272.3692  4109.8267.4965  4161.3265.1403
  4304.8257.3528  4395.8  254.75  4473.8  246.87  4601.3  243.16  4800.2  241.75
  4849.7  246.16    4971  246.84  4991.8  236.07    4997  236.07  4999.8  235.57
    5003  236.07  5020.7   245.9  5219.7  245.82  5462.3  267.88  5541.8  280.56
#Mann= 7 ,-1 , 0
  3725.1     .12       0  3972.7     .07       0  4109.8     .05       0
  4161.3     .07       0  4304.8     .12       0    4997     .07       0
    5003     .12       0
Bank Sta=4971,5020.7
XS Rating Curve= 0 ,0
Exp/Cntr=0.3,0.1

Type RM Length L Ch R = 1 ,35216   ,599,599,599
BEGIN DESCRIPTION:
Mapping XS ad016f22
END DESCRIPTION:
XS GIS Cut Line= 3
      3723512.65     10622052.99      3724283.48     10622506.12
      3724912.51     10623306.71
#Sta/Elev= 30
  3990.8  300.94  4117.1  297.71  4410.7282.6603  4533.1  275.15  4564.4   270.3
  4607.4  268.82  4683.4256.7135  4776.1  244.14  4820.3  241.68  4955.8  245.49
  4970.2  244.16  4984.7  242.68  4991.9  235.37    4997     235  4999.8   234.5
    5003     235    5020  238.06  5028.1  243.49  5034.4  244.17  5042.5  244.49
  5048.9  241.57  5063.3  244.92  5106.3   245.8  5226.9  244.97  5255.8  241.78
  5291.1  241.99  5419.4  250.83    5548255.7255  5789.9  279.86  5903.1  284.63
#Mann= 6 ,-1 , 0
  3990.8     .12       0  4410.7     .07       0  4683.4     .12       0
    4997     .07       0    5003     .12       0    5548     .05       0
Bank Sta=4970.2,5034.4
XS Rating Curve= 0 ,0
Exp/Cntr=0.3,0.1

Type RM Length L Ch R = 1 ,34617   ,556,556,556
BEGIN DESCRIPTION:
TOWN CREEK 44.0
END DESCRIPTION:
XS GIS Cut Line= 3
      3723899.65     10622710.22      3724299.61     10623010.19
       3724599.6     10623310.18
#Sta/Elev= 30
  4494.5  277.09  4563.4270.5164  4616.3  263.84  4687.2  258.75  4716.3  252.95
  4737.2  252.53  4751.7  247.59  4772.6  247.21  4803.8242.3633  4894.5  244.92
    4908  242.93  4916.3  238.56  4922.6  238.81  4930.9   234.2  4951.7  234.52
    4958  236.52  4966.3  234.38  4972.6  242.03  4980.9  240.14  4987.2  242.42
  4991.3  234.18    4997  234.18  4999.8  233.68    5003  234.18  5022.7  234.23
  5036.9  243.15  5107.6  244.23    5227 252.992  5291.4  259.39  5418.7  278.13
#Mann= 6 ,-1 , 0
  4494.5     .07       0  4563.4     .16       0  4803.8     .12       0
    4997     .07       0    5003     .12       0    5227     .05       0
Bank Sta=4987.2,5036.9
XS Rating Curve= 0 ,0
Exp/Cntr=0.3,0.1

Type RM Length L Ch R = 1 ,34061   ,477,477,477
BEGIN DESCRIPTION:
TOWN CREEK 43.0
END DESCRIPTION:
XS GIS Cut Line= 3
      3723699.59     10622760.15      3723899.61     10623310.19
      3724249.62     10623510.19
#Sta/Elev= 30
  4388.7  280.05  4484.5  271.68  4527.1  265.79  4557.8259.3976  4622.8  248.68
  4657.1246.8741  4724.6   243.1  4749.9     245  4785.8  242.75  4801.3244.1543
  4841.6  242.76  4928.1   244.8  4976.9  243.94  4987.7  241.57    4997  233.28
  4999.8  232.78    5003  233.28  5025.1  233.28  5040.9  243.36  5058.9246.0886
  5068.3  247.79  5084.1  246.94  5089.9  248.63  5123.4248.5043  5158.3  257.13
  5234.9262.1947  5310.1  270.38    5326  270.01  5331.7   271.8  5377.1  274.89
#Mann= 9 ,-1 , 0
  4388.7     .07       0  4557.8     .16       0  4657.1     .07       0
  4801.3     .12       0    4997     .07       0    5003     .12       0
  5058.9     .05       0  5123.4     .07       0  5234.9     .05       0
Bank Sta=4976.9,5040.9
XS Rating Curve= 0 ,0
Exp/Cntr=0.3,0.1

Type RM Length L Ch R = 1 ,33584   ,1101,1101,1101
BEGIN DESCRIPTION:
TOWN CREEK 42.0
END DESCRIPTION:
XS GIS Cut Line= 3
       3722986.6     10622709.24       3723674.1     10623636.32
      3725152.28     10623865.34
#Sta/Elev= 30
  4122.8  273.65  4144.1273.2544  4218.8  270.64  4249.7266.0183  4318.9  257.43
  4395.5  253.66  4719.6  238.49  4896.9  244.37    4970  243.18    4983  241.28
  4990.8  233.87    4997  232.15  4999.8  231.65    5003  232.15  5026.3  245.44
  5039.1243.5255  5149.6243.3273  5343.3   237.3  5459.9240.5607  5493.6242.5023
  5530.7  249.83  5646.9  263.05  5656.7  267.04  5661.8  263.05  5667.1  268.17
  5687.3  269.99  6123.1  289.56  6312.1  291.09  6579.4  287.99  6772.8   281.2
#Mann= 10 ,-1 , 0
  4122.8     .16       0  4144.1     .05       0  4249.7     .07       0
  4395.5     .12       0    4997     .07       0    5003     .12       0
  5039.1     .07       0  5149.6     .05       0  5459.9     .16       0
  5493.6     .05       0
Bank Sta=4970,5026.3
XS Rating Curve= 0 ,0
Exp/Cntr=0.3,0.1

Type RM Length L Ch R = 1 ,32483   ,550,550,550
BEGIN DESCRIPTION:
TOWN CREEK 41.0
END DESCRIPTION:
XS GIS Cut Line= 4
      3722804.31     10622756.12      3723043.89     10623521.74
       3723361.6     10623886.32      3723450.14     10625651.98
#Sta/Elev= 30
  4056.4  283.27  4120.8282.4431  4224.9 279.761  4321.3  269.95  4396.7   255.1
  4536.6248.7866  4726.6  249.53    4982  242.33    4997  229.94  4999.8  229.44
    5003  229.94  5031.4  241.44  5080.4239.9875  5249.9241.2066    5278240.8514
  5373.1 243.505  5471.5246.2163  5569.9 243.909  5596.4  243.15  5626.4  230.69
  5646.5  240.88  5726.6     240  5766.7247.4663    5865262.1146  5961.2264.6149
  5963.4264.7095  6061.8271.1412  6577.6  284.06  6817.9  282.61  7110.1  293.33
#Mann= 17 ,-1 , 0
  4056.4     .12       0  4120.8     .16       0  4224.9     .07       0
  4536.6     .12       0    4997     .07       0    5003     .12       0
  5080.4     .05       0  5249.9     .16       0    5278     .07       0
  5373.1     .05       0  5471.5     .07       0  5569.9     .12       0
  5766.7     .05       0    5865     .08       0  5961.2     .07       0
  5963.4     .08       0  6061.8     .05       0
Bank Sta=4982,5031.4
XS Rating Curve= 0 ,0
Exp/Cntr=0.3,0.1

Type RM Length L Ch R = 1 ,31933   ,983,983,983
BEGIN DESCRIPTION:
TOWN CREEK 40.0
END DESCRIPTION:
XS GIS Cut Line= 3
      3722720.98     10623214.47      3722892.85     10624256.12
      3723204.59     10625295.23
#Sta/Elev= 30
  4305.2  269.92  4544.1  257.39    4838  251.31  4929.2  243.79  4943.1  244.95
  4949.5  241.76  4959.7  241.63  4979.9  239.51  4990.1  229.68    4997  228.77
  4999.8  228.27    5003  228.77  5010.3  229.46  5020.5  237.06  5040.7  240.89
  5119.9239.0863  5386.3 239.735  5459.1  241.03  5501.7237.8887  5553.1  239.68
  5584.4  245.51  5605.3  241.67  5711.4242.9232  5852.5  254.59  5857.7  259.11
  5866.3  260.97    5916265.3357  6016.4273.3887  6283.9  284.21  6445.8  286.62
#Mann= 10 ,-1 , 0
  4305.2     .12       0    4997     .07       0    5003     .12       0
  5119.9     .16       0  5386.3     .12       0  5501.7     .05       0
  5605.3     .12       0  5711.4     .05       0    5916     .08       0
  6016.4     .05       0
Bank Sta=4959.7,5040.7
XS Rating Curve= 0 ,0
Exp/Cntr=0.3,0.1

Type RM Length L Ch R = 1 ,30950   ,544,544,544
BEGIN DESCRIPTION:
TOWN CREEK 39.0
END DESCRIPTION:
XS GIS Cut Line= 3
      3722559.51     10623136.34      3722356.39     10623855.07
       3722236.6     10625151.97
#Sta/Elev= 30
  4149.3  266.52  4168.3264.2714    4297 254.621  4353.6  252.98  4392.7  248.44
  4547.5244.3802  4753.2  237.79  4787.2   240.8  4865.5  241.47    4916  238.92
  4941.5  242.14  4961.6  239.45  4996.2227.6841    4997  227.66  4999.8  227.16
    5003  227.66  5020.6  238.93  5182.5  241.03  5202.6  237.76  5252.8  236.35
  5282.9  236.71    5312241.2193  5343.2  241.23  5349.3   238.2  5398.3239.1838
  5453.7  239.53  5568.5     247  5684.6  256.67  5892.3  279.53  6198.6   287.1
#Mann= 9 ,-1 , 0
  4149.3     .07       0  4168.3     .12       0    4297     .05       0
  4547.5     .12       0  4996.2     .16       0    4997     .07       0
    5003     .16       0    5312     .08       0  5398.3     .05       0
Bank Sta=4941.5,5020.6
XS Rating Curve= 0 ,0
Exp/Cntr=0.3,0.1

Type RM Length L Ch R = 1 ,30406   ,606,606,606
BEGIN DESCRIPTION:
TOWN CREEK 38.0
END DESCRIPTION:
XS GIS Cut Line= 3
      3722340.77     10622969.65      3721960.56     10623766.53
      3721013.59      10624370.1
#Sta/Elev= 30
  4370.2  279.99  4429.9278.2689  4514.8  272.88  4590.2  261.39  4625.6  253.03
  4686.5  245.59  4731.9  244.31  4760.1  240.47  4931.4241.6668  4964.3   240.6
  4980.2  229.17    4997  227.21  4999.8  226.71    5003  227.21  5015.2   235.5
  5032.4  239.35  5267.9239.4141  5328.2  239.64  5358.7  233.83  5385.8  234.19
  5401.8 238.551  5422.2  241.97  5437.4  240.99    5444  235.98  5452.6  235.27
  5513.6236.3205  5849.6   243.4  5907.1  247.74  6146.6  276.16  6376.1  287.55
#Mann= 8 ,-1 , 0
  4370.2     .12       0  4429.9     .05       0  4931.4     .16       0
    4997     .07       0    5003     .16       0  5267.9     .12       0
  5401.8     .08       0  5513.6     .05       0
Bank Sta=4964.3,5032.4
XS Rating Curve= 0 ,0
Exp/Cntr=0.3,0.1

Type RM Length L Ch R = 1 ,29800   ,561,561,561
BEGIN DESCRIPTION:
TOWN CREEK 37.0
END DESCRIPTION:
XS GIS Cut Line= 3
      3722249.64     10622860.15      3721649.61     10623560.19
      3720949.62     10624310.18
#Sta/Elev= 30
  4101.1  287.13  4136.8  284.32  4249.9  257.34  4378.9240.5917  4427.7  236.56
  4518.7 237.449  4547.6237.9795  4643.8239.6527  4706.7239.5566  4966.6  239.13
  4980.8  236.42  4987.4  227.23    4997  226.69  4999.8  226.19    5003  226.69
  5009.4  227.22  5014.8233.4789    5016  234.87    5025  235.22  5058.5  238.78
  5079.5  244.35  5129.4  244.21  5136.2  247.57  5148.2248.3206  5176.2253.1244
  5284.7  254.02  5454.7  246.85  5518.2  247.84  5815.7  273.31    6049   287.8
#Mann= 12 ,-1 , 0
  4101.1     .12       0  4378.9     .16       0  4518.7     .05       0
  4547.6     .16       0  4643.8      .1       0  4706.7     .07       0
    4997     .07       0    5003     .07       0  5014.8     .12       0
    5025     .05       0  5148.2     .08       0  5176.2     .05       0
Bank Sta=4966.6,5016
XS Rating Curve= 0 ,0
Exp/Cntr=0.3,0.1

Type RM Length L Ch R = 1 ,29239   ,605,605,605
BEGIN DESCRIPTION:
TOWN CREEK 36.0
END DESCRIPTION:
XS GIS Cut Line= 3
      3722249.62     10622810.18      3721649.61     10623010.19
      3720849.58     10623610.21
#Sta/Elev= 30
  4376.6  288.03  4408.2  286.18  4576.9  257.02  4587.4  252.08    4598  250.98
  4629.6  241.47  4650.7  238.87  4713.9  234.96  4882.5237.9984  4956.4   238.6
  4966.9   235.5  4977.4  226.41    4997  225.66  4999.8  225.16    5003  225.66
  5006.4  229.12  5012.2  229.12  5016.4  237.16  5066.4  239.38  5109.1  236.83
  5152.1 237.513  5216.4  244.07  5316.4  249.62  5430.9  249.69  5509.1   246.9
  5666.4  250.86  5722.6  248.86  5816.4   249.8  5990.4268.5083  6009.1  270.65
#Mann= 6 ,-1 , 0
  4376.6     .12       0  4882.5     .16       0    4997     .07       0
    5003     .16       0  5152.1     .05       0  5990.4     .16       0
Bank Sta=4956.4,5016.4
XS Rating Curve= 0 ,0
Exp/Cntr=0.3,0.1

Type RM Length L Ch R = 1 ,28634   ,502,502,502
BEGIN DESCRIPTION:
TOWN CREEK 35.0
END DESCRIPTION:
XS GIS Cut Line= 3
      3721799.57     10622310.21      3721449.61     10622510.19
      3720649.64     10623310.16
#Sta/Elev= 30
    4610  296.11  4676.9  290.53  4735.9  277.32  4741.7  274.34  4828.8   257.3
    4871250.7801  4881.3  248.22  4887.1  243.93  4897.2  242.21  4902.9  238.09
  4924.5  234.41  4964.3 235.784  4983.6  236.73    4990  232.67    4997  224.67
  4999.8  224.17    5003  224.67  5016.6   224.7  5041.4  234.87  5069.6  235.39
  5083.8  238.84  5097.6238.5855  5281.8  236.41  5394.9  237.83    5508  236.63
  5677.7  245.44    5760245.8412    5802245.2162  5861.6  245.45  6144.4  262.61
#Mann= 8 ,-1 , 0
    4610     .12       0    4871     .16       0  4964.3      .1       0
    4997     .07       0    5003      .1       0  5097.6     .05       0
    5760     .08       0    5802     .05       0
Bank Sta=4983.6,5041.4
XS Rating Curve= 0 ,0
Exp/Cntr=0.3,0.1

Type RM Length L Ch R = 1 ,28132   ,575,575,575
BEGIN DESCRIPTION:
TOWN CREEK 34.0
END DESCRIPTION:
XS GIS Cut Line= 3
      3721649.65     10622160.19      3721149.61     10622160.19
      3720549.63     10622960.16
#Sta/Elev= 30
  4518.5  288.91  4568.5  282.14  4608.5  273.65  4688.6262.3151  4798.5  246.52
  4818.5  242.34  4858.5  238.22  4948.5  236.77  4968.5  238.38  4988.5  236.32
    4997  223.99  4999.8  223.49    5003  223.99  5010.1 224.342  5040.4  230.27
  5046.7  234.09  5075.8  238.47  5240.4  236.85  5332.1  233.66  5375.8  237.22
  5461.2  238.84  5740.4   235.3  5768.5  236.67  5818.5  242.96  5857.8244.5497
  5868.5  244.05  5882.1  247.26  5959.2 253.629  5975.8  256.27  6018.5  257.65
#Mann= 7 ,-1 , 0
  4518.5     .12       0  4688.6     .16       0    4997     .07       0
    5003     .16       0  5010.1     .05       0  5857.8     .08       0
  5959.2     .05       0
Bank Sta=4968.5,5075.8
XS Rating Curve= 0 ,0
Exp/Cntr=0.3,0.1

Type RM Length L Ch R = 1 ,27557   ,559,559,559
BEGIN DESCRIPTION:
TOWN CREEK 33.0
END DESCRIPTION:
XS GIS Cut Line= 3
      3721149.59     10621210.23      3720899.61     10621760.19
      3719449.61     10623310.18
#Sta/Elev= 30
  4371.8  285.07    4391283.3652  4455.2  272.38  4470.6  272.62  4478.3  268.85
  4668.3  253.15  4712.3  237.57  4734.2  234.25  4840.8   236.8    4877  234.31
  4961.6  237.14  4979.3  234.79    4983  224.14    4997  223.57  4999.8  223.07
    5003  223.57  5018.2  229.18  5022.9234.3176  5025.5  237.16  5159.8     234
  5202.3  237.46  5308.3  235.11  5435.8  235.99  5478.3  233.27  5563.3  236.12
  5881.3  233.87  5973.6  238.39  6016.1  237.24  6553.5  261.04  7098.4  296.97
#Mann= 5 ,-1 , 0
  4371.8     .12       0    4391     .16       0    4997     .07       0
    5003     .16       0  5022.9     .05       0
Bank Sta=4961.6,5025.5
XS Rating Curve= 0 ,0
Exp/Cntr=0.3,0.1

Type RM Length L Ch R = 1 ,26998   ,1011,1011,1011
BEGIN DESCRIPTION:
TOWN CREEK 32.0
END DESCRIPTION:
XS GIS Cut Line= 3
      3720749.61      10621060.2      3720649.61     10621460.19
       3719649.6      10623010.2
#Sta/Elev= 30
    4567  286.22  4639.1  281.18  4705.1271.6683  4762.8  262.74  4927.8  242.51
  4938.1  241.02  4948.4  236.72  4961.3  236.51  4976.7  231.61  4982.3  231.61
  4986.9  223.03    4997  222.91  4999.8  222.41    5003  222.91    5008  222.91
  5012.4226.8511  5024.6236.3014  5029.1  236.82  5136.7 237.131  5304.3  235.22
  5522.1   235.4  5673.3  232.74  5745.8   235.7  5969.6  234.91  6116.4237.0689
  6160.2237.6524  6324.1   241.2  6468.5  250.51    6650  259.43  6823.9  272.46
#Mann= 9 ,-1 , 0
    4567     .12       0  4705.1     .16       0    4997     .07       0
    5003     .16       0  5012.4     .12       0  5024.6     .16       0
  5136.7     .05       0  6116.4     .08       0  6160.2     .05       0
Bank Sta=4961.3,5029.1
XS Rating Curve= 0 ,0
Exp/Cntr=0.3,0.1

Type RM Length L Ch R = 1 ,25987   ,548,548,548
BEGIN DESCRIPTION:
TOWN CREEK 31.0
END DESCRIPTION:
XS GIS Cut Line= 3
      3720485.72     10621143.42      3720092.48      10621557.6
       3718783.5     10622073.75
#Sta/Elev= 30
  4387.4  281.38  4411.1279.7725  4523.7   266.6    4531  263.71  4615.9  250.06
  4707.8  237.34  4856.2   233.5  4972.4  235.24  4978.5  234.23    4997  221.79
  4999.8  221.29    5003  221.79  5008.2  221.79  5026.1  228.69  5032.6  236.12
  5034.2 236.037  5146.3  231.01  5294.8  233.32  5338.4  231.56  5348.6  228.56
  5362.8  231.51  5500.8  233.78  5549.6  240.91    5712  250.83  5747.1  250.91
  5767.3254.8966  5875.3 258.975  5933.9  257.71    6126  263.14  6365.6  276.48
#Mann= 7 ,-1 , 0
  4387.4     .12       0  4411.1     .16       0    4997     .07       0
    5003     .16       0  5034.2     .05       0  5767.3     .08       0
  5875.3     .05       0
Bank Sta=4972.4,5032.6
XS Rating Curve= 0 ,0
Exp/Cntr=0.3,0.1

Type RM Length L Ch R = 1 ,25439   ,516,516,516
BEGIN DESCRIPTION:
TOWN CREEK 30.0
END DESCRIPTION:
XS GIS Cut Line= 3
      3720450.77     10621059.67      3719578.25      10621236.5
      3718703.99     10621682.93
#Sta/Elev= 30
  4513.2  279.51  4591.1  268.02  4641.8  263.32  4718.4   251.3  4743.2  250.04
  4839.4  237.51  4902.1  233.29  4953.1  234.87  4963.3  233.79  4973.5  226.99
  4983.7  223.05    4997  221.42  4999.8  220.92    5003  221.42  5014.3  229.29
  5024.5  233.31  5033.3233.3783  5157.2  234.46  5259.2  230.48  5320.4  231.49
  5340.9  229.81  5458.1  235.23  5637.3  247.18  5761.2  250.44  5998.5  264.64
  6053.2  262.84  6075.6  265.12  6087.4  269.63  6187.2  271.88  6385.1  270.69
#Mann= 4 ,-1 , 0
  4513.2     .16       0    4997     .07       0    5003     .16       0
  5033.3     .05       0
Bank Sta=4953.1,5024.5
XS Rating Curve= 0 ,0
Exp/Cntr=0.3,0.1

Type RM Length L Ch R = 1 ,24923   ,1109,1109,1109
BEGIN DESCRIPTION:
TOWN CREEK 29.0
END DESCRIPTION:
XS GIS Cut Line= 3
      3720555.36     10620865.69      3719843.59     10620839.64
      3718872.94     10621151.64
#Sta/Elev= 30
    4048  273.24  4137.5267.2231  4235.4259.9265    4364  246.84  4373.4246.7366
  4394.8244.7868  4532.4236.2052  4634.1  232.57  4744.2  234.28  4811.4  234.48
  4907.7  232.55    4964  233.86  4977.1   231.9    4985  223.31    4997   220.7
  4999.8   220.2    5003   220.7  5009.2  223.89    5027  229.69  5041.3  230.02
  5068.1  233.24  5098.8236.7431  5105.5   236.2  5137.6  238.53  5303.3  240.47
  5399.6  244.58  5431.7  247.44  5478.7   247.7  5661.6  257.19  5779.8  265.11
#Mann= 9 ,-1 , 0
    4048     .12       0  4137.5     .16       0  4235.4     .12       0
  4373.4     .16       0  4394.8     .12       0  4532.4     .16       0
    4997     .07       0    5003     .16       0  5098.8     .05       0
Bank Sta=4964,5068.1
XS Rating Curve= 0 ,0
Exp/Cntr=0.3,0.1

Type RM Length L Ch R = 1 ,23814   ,532,532,532
BEGIN DESCRIPTION:
TOWN CREEK 28.0
END DESCRIPTION:
XS GIS Cut Line= 3
      3720249.62     10619610.16      3719999.61     10620010.19
      3718699.57     10620960.22
#Sta/Elev= 30
  4549.4  287.14  4666.8  265.55  4876.7  245.39  4897.9  240.52  4903.8  243.77
  4913.2  240.31  4919.1   241.5  4934.5  232.81  4937.3233.8768  4940.3  235.02
  4949.8  230.94  4955.7  232.28    4971  228.23  4985.7  219.61    4997  218.71
  4999.8  218.21    5003  218.71  5013.5  221.43  5018.2  225.06  5028.5  226.39
  5034.7  231.92    5064  230.73  5150.5233.7357  5306.5  235.03  5651.7  232.06
  5973.7  235.39  6059.4   237.5  6159.8  244.92  6352.1  249.92  6631.3     267
#Mann= 5 ,-1 , 0
  4549.4     .12       0  4937.3     .16       0    4997     .07       0
    5003     .16       0  5150.5     .05       0
Bank Sta=4955.7,5034.7
XS Rating Curve= 0 ,0
Exp/Cntr=0.3,0.1

Type RM Length L Ch R = 1 ,23282   ,539,539,539
BEGIN DESCRIPTION:
TOWN CREEK 27.0
END DESCRIPTION:
XS GIS Cut Line= 3
      3719899.61     10619310.18      3719699.61     10619660.19
      3718699.61     10620910.19
#Sta/Elev= 30
  4559.8   278.8  4610.9  276.83  4702.3267.8429  4890.2  245.56  4905.3  243.23
  4911.8  238.28  4917.6  239.71  4927.6  236.53  4933.4  238.61  4939.9  231.68
  4949.2  229.41    4955  230.89  4959.2227.9583  4966.1   227.4  4984.5  219.45
  4990.9  222.88    4997  218.48  4999.8  217.98    5003  218.48  5019.7  218.75
    5027  226.68  5034.2  229.95  5080.6  230.59  5168.6  234.17  5255.1  231.28
    5945  233.43  6037.8  236.26  6172.3  247.77  6393.2  254.71  6563.7  265.88
#Mann= 6 ,-1 , 0
  4559.8     .16       0  4702.3     .12       0  4959.2     .16       0
    4997     .07       0    5003     .16       0  5080.6     .05       0
Bank Sta=4955,5034.2
XS Rating Curve= 0 ,0
Exp/Cntr=0.3,0.1

Type RM Length L Ch R = 1 ,22743   ,525,525,525
BEGIN DESCRIPTION:
TOWN CREEK 26.0
END DESCRIPTION:
XS GIS Cut Line= 3
      3719249.61     10619110.18      3719249.61     10619610.19
      3718699.63     10620710.15
#Sta/Elev= 30
  4548.9  277.06    4593 271.316  4638.9  257.86  4678.9   248.7  4718.9  242.94
  4848.9  228.64  4888.9  231.61  4938.9  232.45  4958.9  226.61  4968.9  218.52
    4997  217.88  4999.8  217.38    5003  217.88  5008.9  220.54  5028.9  224.85
  5057.3  224.17  5062.9  220.48  5071.3  222.27  5079.7  226.63  5085.2  224.58
  5093.6  229.18  5114.9232.3232  5482.1  230.13  5585.6  233.77  5711.3  232.58
  5853.9  235.04  6010.4  242.58  6069.1  251.24    6153  253.45  6278.7  262.16
#Mann= 5 ,-1 , 0
  4548.9     .12       0    4593     .16       0    4997     .07       0
    5003     .16       0  5114.9     .05       0
Bank Sta=4938.9,5028.9
XS Rating Curve= 0 ,0
Exp/Cntr=0.3,0.1

Type RM Length L Ch R = 1 ,22218   ,20,20,20
BEGIN DESCRIPTION:
TOWN CREEK 25.0
END DESCRIPTION:
XS GIS Cut Line= 3
       3719249.6      10619060.2      3718899.61     10619310.19
       3718649.6     10620710.24
#Sta/Elev= 30
  4563.2  279.29  4671.3  275.13  4698.4  268.64  4721.7  266.45  4727.9  263.33
  4742.6  263.61  4763.5  258.59  4772.1  259.03  4813.9  246.15  4828.6  245.94
  4858.1  239.67    4879  238.03  4885.2  233.49  4956.4  229.63  4971.2  222.04
  4985.9  217.71    4997  217.71  4999.8  217.21    5003  217.71  5020.2  228.84
  5027.6229.3849  5054.3  231.51    5147 231.182  5226.9  229.18  5309.7  231.64
  5481.4  229.72  5968.5  235.97  6090.4  242.24  6232.6  257.33  6415.5  265.66
#Mann= 5 ,-1 , 0
  4563.2     .12       0    4997     .07       0    5003     .12       0
  5027.6     .16       0    5147     .05       0
Bank Sta=4956.4,5020.2
XS Rating Curve= 0 ,0
Exp/Cntr=0.3,0.1

Type RM Length L Ch R = 1 ,22198   ,358,358,358
BEGIN DESCRIPTION:
Mapping XS b7b043a8
END DESCRIPTION:
XS GIS Cut Line= 3
      3719099.18     10619139.01      3718883.94      10619288.3
      3718609.64     10620583.42
#Sta/Elev= 30
  4713.1  268.49  4807.8  253.88  4813.8  248.47  4828.7  248.44  4834.8  244.79
  4879.4  241.14  4885.4  238.06  4915.2  236.48  4921.3  233.56    4930  234.89
  4936.1  231.42    4951  232.69  4965.8  228.36  4974.6     219    4997  217.62
  4999.8  217.12    5003  217.62  5016.4  226.31  5021.5  224.51  5036.8228.9415
  5071.2  231.38  5164.8230.3816  5215.2  227.94  5309.4  231.43  5467.6  229.37
  5917.4  235.59  6060.5  240.79  6152.5  249.95  6193.4  258.05  6298.9  263.44
#Mann= 5 ,-1 , 0
  4713.1     .12       0    4997     .07       0    5003     .12       0
  5036.8     .16       0  5164.8     .05       0
Bank Sta=4951,5016.4
XS Rating Curve= 0 ,0
Exp/Cntr=0.3,0.1

Type RM Length L Ch R = 1 ,21840   ,432,432,432
BEGIN DESCRIPTION:
Mapping XS 341f31df
END DESCRIPTION:
XS GIS Cut Line= 3
      3719005.51     10619187.58        3718627.     10619395.93
      3718585.37      10620516.3
#Sta/Elev= 30
  4419.4  253.86  4426.1  251.09  4455.3  248.12    4461  244.72  4514.9  242.77
  4520.6  239.14  4536.7  240.56  4542.4  236.95  4596.4  234.61  4602.1  230.67
  4618.1   232.4  4832.2230.1229  4837.1  227.81  4918.3  232.23  4945.8  230.51
  4975.8   223.6  4985.8  218.21    4997  217.87  4999.8  217.37    5003  217.87
  5035.8  225.26  5065.9  228.92  5095.9   226.8  5155.9  226.83  5188.1  229.66
  5716.3  239.55  5826.4  244.25  5886.4  250.77  5916.5  256.95  5972.6  260.06
#Mann= 4 ,-1 , 0
  4419.4     .12       0  4832.2     .05       0    4997     .03       0
    5003     .05       0
Bank Sta=4945.8,5065.9
XS Rating Curve= 0 ,0
Exp/Cntr=0.3,0.1

Type RM Length L Ch R = 1 ,21408   ,269,269,269
BEGIN DESCRIPTION:
Mapping XS e7455e4a
END DESCRIPTION:
XS GIS Cut Line= 3
      3718942.97     10619173.71      3718356.16     10619420.24
      3718078.39     10619864.68
#Sta/Elev= 30
  4152.9  253.45  4341.9  234.24    4384  238.55  4473.6237.0662  4582.7232.9697
  4590.3  234.93  4595.7  233.36  4619.5  242.16  4677.8  245.15  4701.6  242.14
  4709.7  237.13  4725.4  234.28  4731.4  230.32  4741.8229.7571  4889.2228.5388
  4961.2   231.5  4982.5  224.06  4989.8  217.22    4997  217.06  4999.8  216.56
    5003  217.06    5019     223  5025.2  228.89  5034.3  230.96  5070.9  229.36
  5107.5  232.38  5143.1  241.82  5155.9242.8142  5214.5248.0283  5313.5  249.43
#Mann= 9 ,-1 , 0
  4152.9     .12       0  4473.6     .05       0  4582.7     .08       0
  4741.8     .16       0  4889.2     .12       0    4997     .07       0
    5003     .12       0  5155.9     .16       0  5214.5     .12       0
Bank Sta=4961.2,5034.3
XS Rating Curve= 0 ,0
Exp/Cntr=0.3,0.1

Type RM Length L Ch R = 1 ,21139   ,167,167,167
BEGIN DESCRIPTION:
Mapping XS 1c3ed90e
END DESCRIPTION:
XS GIS Cut Line= 3
       3718897.8     10619152.89      3718123.53     10619395.93
      3717595.76     10619691.06
#Sta/Elev= 30
  4072.3  251.58  4227.6   238.7  4332.1240.9357  4437.1234.9234  4477.3  242.82
  4531.6  245.05  4547.4  238.12  4552.6  238.73  4573.5  231.37  4596.2 230.599
  4617.4   231.8  4649.9  228.99  4762.2  231.33  4856.5  227.86  4880.1229.7716
  4963.5  230.92  4979.5  224.45  4985.2  217.05    4997  216.56  4999.8  216.06
    5003  216.56  5014.3  217.44  5028.6  226.99  5044.6  229.62  5094.5  229.52
  5109.7  236.09  5212.5  259.41  5317.4272.9475  5433.3281.4779  5488.5  282.58
#Mann= 9 ,-1 , 0
  4072.3     .12       0  4332.1     .05       0  4437.1     .08       0
  4596.2     .16       0  4880.1     .12       0    4997     .07       0
    5003     .12       0  5317.4     .16       0  5433.3     .05       0
Bank Sta=4963.5,5044.6
XS Rating Curve= 0 ,0
Exp/Cntr=0.3,0.1

Type RM Length L Ch R = 1 ,20972   ,395,395,395
BEGIN DESCRIPTION:
TOWN CREEK 24.0
END DESCRIPTION:
XS GIS Cut Line= 3
      3718963.79      10619100.8      3718019.36     10619298.71
      3717533.92     10619451.28
#Sta/Elev= 30
  3915.9  262.28  4136.1  240.64  4234.1240.7097    4336236.8225  4359.5  242.44
  4410.6  244.72  4420.3  242.02  4425.4  244.54  4437.9236.8238  4451.5  232.71
  4473.2232.2029  4532.3230.5275  4747.8  227.47  4877.9229.8219  4964.2  231.19
    4997  216.35  4999.8  215.85    5003  216.35  5016.9   216.5  5027.3  224.56
  5048.3  231.15  5066.6  239.47  5131.4  253.91  5136.7  252.84  5159.3259.9649
  5201.5   266.8  5206.7  270.72  5239.1  278.39  5264.2280.3325  5389.7  283.37
#Mann= 11 ,-1 , 0
  3915.9     .12       0  4234.1     .05       0    4336     .08       0
  4437.9     .16       0  4473.2     .08       0  4532.3     .16       0
  4877.9     .12       0    4997     .07       0    5003     .12       0
  5159.3     .16       0  5264.2     .05       0
Bank Sta=4964.2,5048.3
XS Rating Curve= 0 ,0
Exp/Cntr=0.3,0.1

Type RM Length L Ch R = 1 ,20577   ,574,574,574
BEGIN DESCRIPTION:
TOWN CREEK 23.0
END DESCRIPTION:
XS GIS Cut Line= 3
      3719049.61     10619010.19      3717799.61     10618960.19
      3717449.62     10619160.18
#Sta/Elev= 30
  3768.1  277.35  3848.2  270.18  3958.3  252.87  3978.3  253.72  4028.3  247.74
    4159239.0916  4208.5  236.69  4238.5  241.84  4278.5  243.98  4308.5  238.17
  4349.8 234.736  4498.7  228.35  4778.9  231.44    4859  225.05  4911.4226.8456
  4969.1  229.81    4997     216  4999.8   215.5    5003     216  5009.1  216.28
  5016.6   222.1  5032.8  226.82  5076.7  231.09  5107.6  240.68  5247.3  260.75
  5286.9269.1414  5306.3  273.76  5355.3  278.64  5403.4279.5032  5422.2  279.52
#Mann= 8 ,-1 , 0
  3768.1     .12       0    4159     .08       0  4349.8     .16       0
  4911.4     .12       0    4997     .07       0    5003     .12       0
  5286.9     .16       0  5403.4     .05       0
Bank Sta=4969.1,5032.8
XS Rating Curve= 0 ,0
Exp/Cntr=0.3,0.1
