HEC-RAS study ALLIGATOR BRANCH.prj: ALLIGATOR BRANCH Base Level Engineering

--- ALLIGATOR BRANCH.g01 (geometry) --- (continued)

Type RM Length L Ch R = 1 ,77778   ,540,540,540
BEGIN DESCRIPTION:
ALLIGATOR BRANCH 57.0
END DESCRIPTION:
XS GIS Cut Line= 3
      3668949.61     10540360.19      3668199.61     10540160.19
      3666963.57      10539518.7
#Sta/Elev= 30
  4206.3  282.53    4304  277.82  4366.3  272.12  4419.1  267.05    4434  266.99
  4574.4  256.15  4654.6  255.43  4703.1     258  4837.6  257.88  4910.1  255.49
  5164.7  255.39  5167.5  254.89  5170.7  255.39  5288.4  258.27  5309.2  259.35
  5405.4   262.6  5433.2  265.24  5665.4  277.73  5703.6  279.45  5753.7  284.04
  5770.2  284.11  5820.1  288.94  5836.6  289.04  5842.2  290.28  5908.6  294.66
  5962.7  296.95  5974.9  298.66  6074.3  301.96  6199.3  309.13  6375.1  317.24
#Mann= 6 ,-1 , 0
  4206.3     .16       0  4366.3     .12       0  5164.7     .07       0
  5170.7     .12       0  5288.4     .16       0  5665.4     .05       0
Bank Sta=4837.6,5309.2
XS Rating Curve= 0 ,0
Exp/Cntr=0.3,0.1

Type RM Length L Ch R = 1 ,77238   ,520,520,520
BEGIN DESCRIPTION:
ALLIGATOR BRANCH 56.0
END DESCRIPTION:
XS GIS Cut Line= 3
      3669199.57      10539410.2      3668399.61     10539660.19
      3667649.58     10539510.18
#Sta/Elev= 30
  4153.7  283.81  4202.4  282.68  4234.9  279.75  4272.6  278.75  4310.8  275.87
  4331.8  272.26  4342.8  272.91    4370  271.15  4375.2  271.88  4480.5  265.14
  4542.9  262.42  4570.1  260.21  4575.4  260.91  4602.6  259.93  4607.8  260.78
  4635.1  258.42  4640.3  259.73  4656.6  257.75  4672.8  255.63  4845.4  254.91
  4943.1  255.78  5216.2  255.49  5277.4  259.16  5318.2  262.15  5481.3  278.84
  5562.9  285.42  5642.6  294.12  5675.1  296.38  5715.9  301.65  5756.7  304.97
#Mann= 5 ,-1 , 0
  4153.7     .16       0  4480.5     .12       0  4656.6     .07       0
  5277.4     .16       0  5642.6     .05       0
Bank Sta=4656.6,5277.4
XS Rating Curve= 0 ,0
Exp/Cntr=0.3,0.1

Type RM Length L Ch R = 1 ,76718   ,108,108,108
BEGIN DESCRIPTION:
ALLIGATOR BRANCH 55.0
END DESCRIPTION:
XS GIS Cut Line= 4
      3669149.57     10539360.18      3668649.61     10539210.19
      3667999.61     10539110.19      3667465.31     10539515.74
#Sta/Elev= 30
  4483.3  282.39  4598.1   274.2  4637.3  270.03  4642.5  270.38  4660.7   266.4
  4746.9  262.71  4771.1  262.69  4827.8  262.38  4884.3  258.58  4911.3  255.64
  4931.9  254.86  4955.7  255.67  5258.2  255.51  5339.2  258.42  5490.9  272.43
  5511.2  276.12  5565.5  282.05  5628.8  291.77  5688.5  292.82  5755.5  295.08
  5855.3  292.46  5919.8  292.79  5940.6  294.26  5963.4  294.01  6110.8  301.84
    6134  302.53  6140.3   303.9  6163.1  303.15  6190.2  304.65  6333.7  306.56
#Mann= 6 ,-1 , 0
  4483.3     .16       0  4771.1     .12       0  4884.3     .07       0
  5339.2     .16       0  5688.5     .05       0  6110.8     .16       0
Bank Sta=4884.3,5339.2
XS Rating Curve= 0 ,0
Exp/Cntr=0.3,0.1

Type RM Length L Ch R = 1 ,76610   ,46,46,46
BEGIN DESCRIPTION:
Mapping XS cb3e94e3
END DESCRIPTION:
XS GIS Cut Line= 6
      3669184.57     10539349.78      3668773.12      10539172.7
       3668575.2     10538995.62       3668531.8     10538976.52
      3668153.33     10538974.79      3667630.74     10539309.87
#Sta/Elev= 30
  4489.7  283.44  4554.2  280.75  4570.9  277.72  4646.7   273.1  4722.6  264.91
  4814.5  261.97  4853.1  259.93  4911.3  259.81  4936.9   255.3  5023.8   255.2
  5026.6   254.7  5029.8   255.2  5232.8  256.42  5431.8  258.29  5472.9  261.17
  5544.7   267.2  5628.6  277.86    5644  279.19    5650  278.24  5665.2  280.74
  5700.5  283.04  5774.2  286.57  5780.1  288.52  5795.3  287.67  5967.8  293.92
  6055.7   290.2  6111.4  291.55  6178.1  294.61  6231.9  296.28    6250  296.61
#Mann= 11 ,-1 , 0
  4489.7     .16       0  4814.5     .12       0  5023.8     .07       0
  5029.8     .12       0  5232.8     .16       0  5431.8     .05       0
  5700.5     .16       0  5795.3     .05       0  6111.4     .16       0
  6178.1     .05       0  6231.9     .16       0
Bank Sta=4911.3,5472.9
XS Rating Curve= 0 ,0
Exp/Cntr=0.3,0.1

Type RM Length L Ch R = 1 ,76564   ,39,39,39
BEGIN DESCRIPTION:
Mapping XS 2e191667
END DESCRIPTION:
XS GIS Cut Line= 6
      3669197.21     10539331.45        3668843.     10539156.95
      3668587.79     10538966.84      3668496.65     10538927.78
      3668189.35     10538909.55      3667595.58     10539289.77
#Sta/Elev= 30
  4500.6  283.75  4531.4  282.91    4627  274.42  4665.1   272.8  4754.3   263.8
  4839.1  260.23  4931.7  262.95  5032.8  262.38  5188.3  259.19  5196.4  257.61
  5255.4  256.91  5264.6  254.52  5293.8  257.98  5456.9  258.49  5570.5  266.76
  5665.2  278.29  5671.2  277.23  5707.5  280.34  5777.6  281.91  5785.8  282.09
  5895.2  286.74  5925.6  285.69  5931.6  287.21  6025.4  291.28  6143.6  287.86
  6164.9  288.65  6170.9   290.6  6186.1   289.8  6228.4  292.59  6325.9   293.9
#Mann= 8 ,-1 , 0
  4500.6     .16       0  4839.1     .12       0  5188.3     .07       0
  5293.8     .16       0  5456.9     .05       0  5777.6     .16       0
  5785.8     .05       0  6143.6     .16       0
#XS Ineff= 2 ,-1
 4661.36 4922.73265.8279 5222.73 5611.36  265.71
Permanent Ineff=
       F       F
Bank Sta=4931.7,5032.8
XS Rating Curve= 0 ,0
Exp/Cntr=0.3,0.1

Type RM Length L Ch R = 1 ,76525   ,372,372,372
BEGIN DESCRIPTION:
Mapping XS ff6e3cef
END DESCRIPTION:
XS GIS Cut Line= 6
      3669222.81     10539311.61      3668858.19     10539134.51
      3668811.32      10539085.9      3668500.55     10538894.92
      3668373.82     10538757.77       3667689.8     10538521.67
#Sta/Elev= 30
  4494.5  283.82  4596.7  278.18  4760.1  263.37  4854.3  259.98  4916.1  261.73
  4937.2  257.26    4965  255.67  4967.4  255.67  5008.4  252.93    5030   255.2
  5118.8  257.25  5124.7  255.84  5155.5  257.72  5161.4  256.59  5192.2  259.33
  5213.5  257.55  5273.6  257.16  5292.8   255.7  5314.1  259.25  5385.7  259.88
    5393  255.52  5406.7   254.4    5414  258.71  5420.8  257.72  5428.2  260.04
  5914.8  261.44  6062.7  274.98  6158.1  286.73  6189.8  292.95  6242.5  298.61
#Mann= 6 ,-1 , 0
  4494.5     .16       0  4854.3     .12       0    4965     .07       0
    5030     .12       0  5273.6     .16       0  6062.7     .05       0
#XS Ineff= 2 ,-1
 5194.32 5492.05  260.14 5492.05 5977.27  263.33
Permanent Ineff=
       F       F
Bank Sta=4967.4,5030
XS Rating Curve= 0 ,0
Exp/Cntr=0.3,0.1

Type RM Length L Ch R = 1 ,76153   ,418,418,418
BEGIN DESCRIPTION:
ALLIGATOR BRANCH 54.0
END DESCRIPTION:
XS GIS Cut Line= 3
      3670476.47     10539056.39      3668532.06     10538665.78
      3667413.42     10538076.11
#Sta/Elev= 30
  3369.2  307.13  3617.9  299.57  3702.6  298.48  3794.4  302.59  3896.4  304.19
  4049.4  298.69  4122.7  293.79  4222.8  284.91  4322.9  277.48  4487.6  269.77
    4523  266.37  4702.2  255.31  4823.2  254.35  4894.7  257.71  4977.6  257.11
  5001.3  252.88  5028.6   257.2  5154.2  255.88  5222.4  257.85  5314.2   256.3
  5456.1  258.55  5483.8  257.46    5754  259.73  5979.1  265.62  6083.6  272.65
  6320.2  292.27  6417.8  305.69  6446.8  311.61  6519.6  320.57    6617  323.53
#Mann= 10 ,-1 , 0
  3369.2     .16       0  3617.9     .05       0  4122.7     .16       0
  4222.8     .12       0  4322.9     .16       0    4523     .05       0
  4823.2     .12       0  4977.6     .05       0  5028.6     .05       0
    5754     .16       0
#XS Ineff= 1 ,-1
 5593.18 5959.09  263.82
Permanent Ineff=
       F
Bank Sta=4977.6,5028.6
XS Rating Curve= 0 ,0
Exp/Cntr=0.3,0.1

Type RM Length L Ch R = 1 ,75735   ,97,97,97
BEGIN DESCRIPTION:
ALLIGATOR BRANCH 53.0
END DESCRIPTION:
XS GIS Cut Line= 6
      3670152.36     10538804.08      3669687.04     10538831.86
      3669225.23     10538508.94       3668829.4     10538196.44
      3668482.18      10537939.5      3667846.74      10537449.9
#Sta/Elev= 30
  3707.2  313.48  3714.6  313.35  3889.4   310.3  4050.6  299.59  4110.7  292.71
  4227.1  285.73    4306  278.26  4487.6  261.39  4668.8  252.14  4689.9  253.91
  4982.4  256.43  4988.7  254.38  5003.2  253.94  5024.3  256.18  5060.9  255.73
  5075.3  253.56  5096.2  255.71  5266.1  253.15  5380.9  255.82  5631.4  257.68
  5671.6  261.25  5681.4  259.97  5695.9  263.84  5710.4  264.75  5716.8  263.05
  5745.8  264.28  5895.2  273.12  6023.9  275.96    6109  280.56  6475.3  293.33
#Mann= 6 ,-1 , 0
  3707.2     .16       0  3714.6     .05       0  4227.1     .16       0
    4306     .05       0  4982.4     .03       0  5024.3     .05       0
Bank Sta=4982.4,5024.3
XS Rating Curve= 0 ,0
Exp/Cntr=0.3,0.1

Type RM Length L Ch R = 1 ,75638   ,479,479,479
BEGIN DESCRIPTION:
Mapping XS a4615864
END DESCRIPTION:
XS GIS Cut Line= 6
      3670141.88     10538692.97      3669770.37     10538727.69
      3669371.07     10538508.94      3669006.48      10538213.8
      3668447.46     10537758.94      3668127.99     10537408.23
#Sta/Elev= 30
  3777.5  318.96    3820  316.67  3900.3  315.52  3920.4  313.32    4071  306.39
  4156.5  299.77  4379.3  271.65  4516.4  258.26  4641.8  254.55  4662.6  252.26
  4720.2  254.33  4961.6  254.74  4982.4     251  5001.7  249.57  5025.5  249.69
  5039.9  254.91  5225.2  254.12  5260.4  252.13  5289.2  253.92  5565.6  254.19
  5679.1  256.37  5786.1  263.21  5791.1  264.91  5906.4  273.94  5977.4  277.25
  6083.5  288.15  6118.7  294.21  6154.4  297.95  6211.2  299.59  6270.1  297.67
#Mann= 3 , 0 , 0
  3777.5     .05       0  4961.6     .03       0  5039.9     .05       0
Bank Sta=4961.6,5039.9
XS Rating Curve= 0 ,0
Exp/Cntr=0.3,0.1

Type RM Length L Ch R = 1 ,75159   ,670,670,670
BEGIN DESCRIPTION:
ALLIGATOR BRANCH 52.0
END DESCRIPTION:
XS GIS Cut Line= 3
       3670049.6     10538310.18      3669299.61     10537910.19
      3668149.65     10537360.21
#Sta/Elev= 30
  4158.1  314.09  4188.2  312.27  4232.1  305.03  4254.1  303.71  4260.1  301.31
  4292.3  295.61  4328.1  291.88  4336.2  289.64    4446  279.41  4478.6  274.89
  4588.4  265.06  4742.1  255.59  4890.2  252.78  4994.3  254.17  5022.2  252.59
  5030.3     254  5158.2  251.68  5407.1   252.1  5426.3  251.04  5451.5  252.31
  5736.2   253.6  5758.8  257.03  5817.3  259.27  5951.3  270.92  6087.4  286.26
    6110  289.26  6116.6  291.61    6172  298.51  6228.9  302.15  6282.8  301.12
#Mann= 4 ,-1 , 0
  4158.1     .16       0  4478.6     .05       0  5407.1     .03       0
  5451.5     .05       0
Bank Sta=4994.3,5030.3
XS Rating Curve= 0 ,0
Exp/Cntr=0.3,0.1

Type RM Length L Ch R = 1 ,74489   ,399,399,399
BEGIN DESCRIPTION:
ALLIGATOR BRANCH 51.0
END DESCRIPTION:
XS GIS Cut Line= 3
      3669849.66      10537510.2      3669009.49     10537346.33
      3668249.65      10537160.2
#Sta/Elev= 30
  4154.2  278.62  4185.1  275.82  4215.4  274.88  4256.1  270.41  4307.1  267.53
  4339.9  264.64  4347.8  262.64  4386.4  258.65  4541.2  257.32  4597.9     258
  4948.9  251.84  5012.6  250.41  5020.4  251.91    5154  249.88  5288.1  251.15
  5380.7  256.71  5421.9  261.02  5436.3  261.34    5494   266.9  5545.5  272.91
  5561.1  275.73  5566.3  275.42  5576.3  277.44  5607.9  280.22  5627.8  283.26
  5644.4  287.51  5649.5  287.35    5686  294.07  5741.1  300.66  5792.5  304.87
#Mann= 3 , 0 , 0
  4154.2     .05       0  4948.9     .03       0  5020.4     .05       0
Bank Sta=4948.9,5020.4
XS Rating Curve= 0 ,0
Exp/Cntr=0.3,0.1

Type RM Length L Ch R = 1 ,74090   ,504,504,504
BEGIN DESCRIPTION:
ALLIGATOR BRANCH 50.0
END DESCRIPTION:
XS GIS Cut Line= 3
      3670449.58      10536460.2      3668899.61     10537010.19
      3668249.62     10537110.19
#Sta/Elev= 30
  3379.3   335.2  3464.2  332.63  3506.6  329.71  3616.6  314.58  3667.2  307.57
  3810.9  291.95  3909.8  284.16  4100.8  273.93  4227.2  269.23  4319.8  264.12
  4474.1  262.71  4592.3  258.45  4741.3   256.5  4946.8  251.71  5008.3  248.46
  5011.5  248.96  5013.8  250.85  5104.9  249.31  5216.2  250.35  5257.9  252.65
  5297.1  257.71  5321.2  259.15  5398.3  268.47  5452.7  273.65    5459  275.43
  5550.1  287.96  5579.2  294.23  5600.7  297.15  5661.4   303.4  5681.6  304.14
#Mann= 4 ,-1 , 0
  3379.3     .16       0  3616.6     .05       0  4946.8     .03       0
  5013.8     .05       0
Bank Sta=4946.8,5013.8
XS Rating Curve= 0 ,0
Exp/Cntr=0.3,0.1

Type RM Length L Ch R = 1 ,73586   ,520,520,520
BEGIN DESCRIPTION:
ALLIGATOR BRANCH 49.0
END DESCRIPTION:
XS GIS Cut Line= 3
      3670349.64     10536410.19      3668949.61     10536510.19
      3668299.62     10536910.18
#Sta/Elev= 30
  3556.4  330.74  3616.6   324.8    3656  319.09  3716.8  310.06  3817.1  299.18
  3909.8  292.42  3997.5  282.36  4077.8  276.38  4248.2   268.7  4418.6  263.75
  4611.6  262.66  4689.3  260.45  4892.3   249.3  4962.9  250.07  4967.7  246.69
  4973.6  248.07  4982.9  246.15  4986.1  246.65    4989  249.51  4995.2  246.94
  5004.4  249.65  5010.3  247.99  5018.7  249.83    5273  253.39  5300.5  252.42
  5352.2  254.39  5504.9  267.03  5599.6   278.6  5694.2  293.62  5723.2  296.55
#Mann= 4 ,-1 , 0
  3556.4     .16       0    3656     .05       0  4962.9     .05       0
  5018.7     .05       0
Bank Sta=4962.9,5018.7
XS Rating Curve= 0 ,0
Exp/Cntr=0.3,0.1

Type RM Length L Ch R = 1 ,73066   ,610,610,610
BEGIN DESCRIPTION:
ALLIGATOR BRANCH 48.0
END DESCRIPTION:
XS GIS Cut Line= 3
      3669999.63     10536260.19      3669199.61     10536110.19
      3668399.58     10535510.16
#Sta/Elev= 30
  4157.6  290.26    4178  288.59  4183.9  286.91  4346.7  273.74  4523.9  262.15
  4686.7  253.38  4899.4  249.68  4993.4  249.34  4996.7  246.08  4999.4  245.58
    5008  246.32  5014.3  249.24  5021.6  249.91  5049.7  248.71  5114.3  249.42
  5164.3  248.57  5287.3  250.69  5314.3  250.85  5321.6  251.97  5371.6  253.51
  5564.3  264.49  5585.1  267.25  5621.6   269.1    5758  281.56  5785.1  282.62
  5849.7  289.24    5858  291.44  5871.6  291.13  5943.4  299.33  5971.6   301.2
#Mann= 5 ,-1 , 0
  4157.6     .05       0  4899.4     .16       0  4993.4     .07       0
  5021.6     .16       0  5287.3     .05       0
Bank Sta=4993.4,5021.6
XS Rating Curve= 0 ,0
Exp/Cntr=0.3,0.1

Type RM Length L Ch R = 1 ,72456   ,565,565,565
BEGIN DESCRIPTION:
ALLIGATOR BRANCH 47.0
END DESCRIPTION:
XS GIS Cut Line= 3
      3670299.57     10536360.16      3669499.61     10535810.19
      3668699.61     10535260.19
#Sta/Elev= 30
  3996.8  322.93  4037.2  316.99  4147.6   304.5  4198.4  301.01  4255.2  294.08
    4291  290.63  4299.9  290.93  4312.3  288.62    4494  270.63  4788.4  250.64
  4873.5  247.72  4939.2  247.67    4975  245.79    4996  246.61  5003.7  244.95
  5010.9  245.66  5016.9  247.92  5046.7   247.1  5067.7  248.98    5205  249.29
  5370.8  252.17  5396.7   253.4  5665.1   265.9  5700.9  269.47  5730.7  271.48
  5736.8  270.85  5751.7  273.19    5817  277.13  5895.1  286.69  5938.4  289.76
#Mann= 7 ,-1 , 0
  3996.8     .16       0  4037.2     .05       0  4788.4     .16       0
    4996     .07       0  5016.9     .05       0  5370.8     .16       0
  5396.7     .05       0
Bank Sta=4939.2,5016.9
XS Rating Curve= 0 ,0
Exp/Cntr=0.3,0.1

Type RM Length L Ch R = 1 ,71891   ,271,271,271
BEGIN DESCRIPTION:
ALLIGATOR BRANCH 46.0
END DESCRIPTION:
XS GIS Cut Line= 3
      3670399.62      10536310.2      3669849.61     10535510.19
      3668399.61     10535110.19
#Sta/Elev= 30
  4008.3  326.45  4136.5  311.68  4383.1  286.21  4490.7  278.42  4613.1  273.43
  4777.5   255.4  4821.4  252.94  4858.9   248.7  4971.7  247.91  4989.5  247.53
  4996.3  247.63  5001.3  244.94  5020.6  247.99  5088.1  248.32  5155.5  249.34
  5176.2  251.74  5223.2  250.12  5228.4  251.65  5262.8  252.29  5302.3  250.27
  5539.3  252.84    5809  260.75  5864.5  264.73  5881.6  267.94  5938.4  270.48
  5977.9  274.08  5985.4  276.49  6017.5  277.87  6172.1   292.2  6483.3  305.58
#Mann= 6 ,-1 , 0
  4008.3     .16       0  4136.5     .05       0  4858.9     .16       0
  4989.5     .07       0  5020.6     .16       0  5088.1     .05       0
Bank Sta=4971.7,5020.6
XS Rating Curve= 0 ,0
Exp/Cntr=0.3,0.1

Type RM Length L Ch R = 1 ,71620   ,921,921,921
BEGIN DESCRIPTION:
ALLIGATOR BRANCH 45.0
END DESCRIPTION:
XS GIS Cut Line= 3
      3671544.24     10535401.89       3670077.2      10535306.4
       3668454.3     10534933.22
#Sta/Elev= 30
  3423.1  325.48  3488.5  318.29  3758.4  295.32  3838.9  292.01  3908.8     287
  3978.9  286.88  4049.1  289.33  4199.4  286.61  4319.6  280.22  4590.2  257.37
  4640.3  256.43  4756.7  250.39  4988.1  246.34  4993.4  245.15  5003.4  244.48
  5024.2  247.53    5096  247.05  5297.3  250.12  5656.2  254.59  5757.9  257.16
  5800.1  257.96  5906.6  261.33  6057.1  275.73  6132.4  280.07  6238.7  289.12
  6245.2  288.15  6286.7  290.02  6399.1  298.38    6512  302.87  6558.5  299.81
#Mann= 7 ,-1 , 0
  3423.1     .05       0  3488.5     .16       0  4993.4     .07       0
  5024.2     .16       0  5297.3     .05       0  5757.9     .08       0
  5800.1     .05       0
Bank Sta=4988.1,5024.2
XS Rating Curve= 0 ,0
Exp/Cntr=0.3,0.1

Type RM Length L Ch R = 1 ,70699   ,570,570,570
BEGIN DESCRIPTION:
ALLIGATOR BRANCH 44.0
END DESCRIPTION:
XS GIS Cut Line= 3
      3670199.63      10534710.2      3669849.61     10534510.19
      3669049.58     10533960.17
#Sta/Elev= 30
    4606  286.31  4629.1  285.01  4686.6   278.2  4775.2  264.68  4824.9   259.8
  4847.9  256.03  4861.6  256.03  4914.8  250.93  4928.5  250.87    4958  246.52
  4986.1  246.96  4995.2  243.06  5001.2  244.01  5006.3  247.26  5031.5   248.6
  5045.5  245.96  5058.5   247.6  5081.9  247.92  5174.9  247.22  5295.4  253.01
  5305.6  253.53  5476.6  263.77  5727.6  275.08  5829.1  283.12  5850.1  283.66
  5895.1  288.64  5943.6  292.46  5951.6  294.24  5972.5  294.82    5980  296.54
#Mann= 6 ,-1 , 0
    4606     .16       0  4986.1     .07       0  5006.3     .16       0
  5295.4     .12       0  5305.6     .16       0  5895.1     .05       0
Bank Sta=4986.1,5006.3
XS Rating Curve= 0 ,0
Exp/Cntr=0.3,0.1

Type RM Length L Ch R = 1 ,70129   ,450,450,450
BEGIN DESCRIPTION:
ALLIGATOR BRANCH 43.0
END DESCRIPTION:
XS GIS Cut Line= 3
      3670699.61     10534410.19      3669999.61     10534010.19
      3669599.61     10533560.19
#Sta/Elev= 30
    4187  316.03  4348.2  298.17  4495.8   276.1  4670.7  257.53  4751.4  250.27
  4808.9  246.98    4855  246.13  4904.7  245.88  4947.9  247.49  4985.3  246.23
  4987.3  241.33  4990.1  240.83  5000.3  242.14  5014.6  246.99    5043  246.01
  5057.2  247.15  5106.5  246.61  5149.2  247.88  5220.3  252.49  5327.6  262.77
  5340.7  263.05  5425.1  272.64  5453.6  277.38  5467.8  281.67    5482  283.87
  5488.7  286.38  5510.4   290.1  5531.3  295.44  5559.8   299.2  5595.3  301.33
#Mann= 4 ,-1 , 0
    4187     .16       0  4985.3     .07       0  5014.6     .16       0
  5327.6      .1       0
Bank Sta=4985.3,5014.6
XS Rating Curve= 0 ,0
Exp/Cntr=0.3,0.1

Type RM Length L Ch R = 1 ,69679   ,774,774,774
BEGIN DESCRIPTION:
ALLIGATOR BRANCH 42.0
END DESCRIPTION:
XS GIS Cut Line= 3
       3670823.7     10534403.59      3670146.64     10533648.41
      3669478.22     10533370.63
#Sta/Elev= 30
  4250.7  318.58  4312.5  315.65  4411.9  304.56    4497   299.2  4510.6  296.25
  4524.8  296.53  4808.1  258.86  4921.8  249.35    4936  247.13  4971.1  245.45
  4992.5  240.83    5007  246.33  5042.1  246.63  5048.8  245.42  5056.3   246.4
    5063   244.4  5089.3  245.94  5254.4  246.74  5315.9  248.58  5377.6  252.44
  5466.2  259.35    5512  265.08  5565.2  269.83  5588.3  273.47  5642.2  279.25
  5689.9  286.66  5695.3  286.16  5759.9  291.63    5820  295.17  5988.8  301.01
#Mann= 7 ,-1 , 0
  4250.7     .16       0  4971.1     .07       0    5007     .16       0
  5089.3     .05       0  5377.6     .16       0  5466.2     .05       0
  5588.3      .1       0
Bank Sta=4971.1,5007
XS Rating Curve= 0 ,0
Exp/Cntr=0.3,0.1

Type RM Length L Ch R = 1 ,68905   ,624,624,624
BEGIN DESCRIPTION:
ALLIGATOR BRANCH 41.0
END DESCRIPTION:
XS GIS Cut Line= 3
       3671199.6     10533610.18      3670699.61     10533360.19
      3670199.63     10533010.21
#Sta/Elev= 30
  4471.9  307.06  4506.3  301.63    4539  297.27  4569.7  295.46  4592.1   292.3
  4597.7  290.29  4614.4  288.97  4748.6  272.11    4771  268.18  4963.8  248.25
  4972.2  245.29  4999.9  241.95  5008.5  244.39  5016.9  244.97  5059.2  243.64
  5095.3  244.74  5131.7  245.75  5212.8  247.62  5267.6   249.2  5282.4  248.53
  5374.9  252.25  5397.1  255.32  5433.7  257.85  5446.4   259.9  5469.9  259.66
    5476  260.62  5482.5  263.85  5565.3  273.55  5627.7   277.6  5641.2  277.63
#Mann= 8 ,-1 , 0
  4471.9     .05       0  4506.3     .16       0  4963.8     .07       0
  5008.5     .16       0  5095.3     .05       0  5131.7     .16       0
  5212.8     .05       0  5565.3     .16       0
Bank Sta=4963.8,5008.5
XS Rating Curve= 0 ,0
Exp/Cntr=0.3,0.1

Type RM Length L Ch R = 1 ,68281   ,504,504,504
BEGIN DESCRIPTION:
ALLIGATOR BRANCH 40.0
END DESCRIPTION:
XS GIS Cut Line= 3
      3671499.64     10533460.22      3670999.61     10533010.19
      3670699.62     10532210.21
#Sta/Elev= 30
  4283.6   327.2  4311.7  324.29  4325.9  320.79  4382.7  312.48  4404.4  307.42
  4411.1  308.07  4467.9  300.33  4488.8  299.27  4496.3  297.08  4552.7  291.83
  4559.8  289.74  4637.5  283.42    4732  270.85  4843.1  260.11    4864  259.67
  4885.7   256.3  4942.5  252.47    4953  249.16    4959  249.16  4966.1  248.16
  4977.7  242.99  4996.1  239.37  5009.7  243.63    5234  247.22  5428.9  257.57
  5459.2  258.87    5469  257.62  5544.6  266.11  5679.9  286.15  5810.7  295.04
#Mann= 4 ,-1 , 0
  4283.6     .05       0    4732     .16       0    4959     .07       0
  5009.7     .16       0
Bank Sta=4959,5009.7
XS Rating Curve= 0 ,0
Exp/Cntr=0.3,0.1

Type RM Length L Ch R = 1 ,67777   ,522,522,522
BEGIN DESCRIPTION:
ALLIGATOR BRANCH 39.0
END DESCRIPTION:
XS GIS Cut Line= 3
       3671499.6     10533410.17      3671299.61     10532660.19
      3670999.61      10532060.2
#Sta/Elev= 30
    4227  321.96  4299.4  315.08  4319.5  310.07  4324.7  310.63  4394.9  301.93
    4465  294.31  4582.1  277.33    4641  268.89  4785.2  255.97  4790.4  254.04
  4837.6  251.84    4876  247.73  4899.7  245.81  4905.5  243.92  4920.4  243.99
  4951.2  238.04  4985.7  241.74    5006  239.42  5025.5  244.96  5047.9  246.26
    5115  244.54  5179.1  246.81  5263.8  253.17  5464.4  267.91  5548.2   278.1
  5562.2  281.18  5615.3  286.46  5620.9  288.78  5651.6  292.14    5674   292.5
#Mann= 8 ,-1 , 0
    4227     .05       0  4394.9     .16       0  4582.1     .05       0
    4876     .16       0  4920.4     .07       0  4985.7     .16       0
  5179.1     .05       0  5263.8     .16       0
Bank Sta=4920.4,5025.5
XS Rating Curve= 0 ,0
Exp/Cntr=0.3,0.1

Type RM Length L Ch R = 1 ,67255   ,402,402,402
BEGIN DESCRIPTION:
ALLIGATOR BRANCH 38.0
END DESCRIPTION:
XS GIS Cut Line= 3
      3671549.61     10532960.21      3671649.61     10532360.19
      3671699.61     10531760.17
#Sta/Elev= 30
  4417.3  264.04  4445.2   260.5    4478     260    4506  256.48  4599.8  249.86
  4727.9  245.81    4833  245.25    4871  243.25  4911.9  243.25    4985  241.38
  4992.4  237.74  5005.3  238.36  5023.1  242.21  5045.7  244.57  5065.7  244.34
  5088.3  246.88  5115.9  246.68    5146  250.56  5186.2  252.37  5196.2  251.83
  5203.7   249.8  5208.7  253.47  5329.1     260    5437  270.87  5444.5  272.84
  5457.1  273.24    5502  278.89  5555.2  287.31  5597.6  295.12  5627.7  298.09
#Mann= 8 ,-1 , 0
  4417.3     .05       0    4478     .12       0  4727.9     .05       0
  4911.9     .16       0    4985     .07       0  5023.1     .16       0
    5502     .12       0  5555.2     .16       0
Bank Sta=4985,5023.1
XS Rating Curve= 0 ,0
Exp/Cntr=0.3,0.1

Type RM Length L Ch R = 1 ,66853   ,784,784,784
BEGIN DESCRIPTION:
ALLIGATOR BRANCH 37.0
END DESCRIPTION:
XS GIS Cut Line= 2
      3672123.65     10534271.58      3671841.52     10531515.48
#Sta/Elev= 30
  3013.3  327.43  3041.3  326.13  3141.4  318.72  3229.9   314.3  3394.2  309.63
  3557.5  311.36  3635.3  314.07  3765.8  313.21  3791.6  314.17  3808.8  311.19
    3839  311.78    3891  307.66  3979.7  292.78    4010  289.72  4160.7  274.76
  4328.4  263.02  4526.4  249.76  4670.8  243.46  4724.5  243.18  4884.4  244.52
  4944.7  243.09  5014.8   237.8  5025.1  242.69  5095.5   243.1    5196  248.05
    5384  265.36  5519.5  281.56  5628.3  291.57  5688.6  299.56  5783.8  300.63
#Mann= 14 ,-1 , 0
  3013.3     .05       0  3041.3      .1       0  3141.4     .16       0
  3229.9     .05       0  3635.3     .16       0  3765.8     .05       0
    4010     .16       0  4328.4     .12       0  4526.4     .05       0
  4724.5     .16       0  4944.7     .07       0  5025.1     .16       0
    5384     .12       0  5519.5     .16       0
Bank Sta=4944.7,5025.1
XS Rating Curve= 0 ,0
Exp/Cntr=0.3,0.1

Type RM Length L Ch R = 1 ,66069   ,1585,1585,1585
BEGIN DESCRIPTION:
ALLIGATOR BRANCH 36.0
END DESCRIPTION:
XS GIS Cut Line= 3
       3672949.6     10533110.17      3672649.61     10532310.19
      3672649.61     10531860.17
#Sta/Elev= 30
    4144  283.36  4208.1   278.3  4214.3     277  4229.4  276.61  4299.7  269.16
  4338.2  266.09  4440.4   256.6  4453.7  256.32  4500.9  252.72  4507.1  251.36
  4566.6  247.43  4635.3  243.23  4688.1  241.99  4794.4  241.64  4842.6  240.54
  4922.7  243.27  4983.3  241.51  5008.1  237.79  5018.4   238.4  5028.4  241.47
  5038.4  242.48  5068.4  241.58  5118.4  246.19  5151.4  250.33  5202.6   258.8
  5228.4  262.59  5258.4  268.77  5298.4  275.38  5358.4  280.92  5448.4  285.14
#Mann= 9 ,-1 , 0
    4144     .16       0  4338.2     .12       0  4566.6     .05       0
  4688.1     .07       0  4794.4     .12       0  4983.3     .07       0
  5028.4     .16       0  5151.4     .12       0  5202.6     .16       0
Bank Sta=4983.3,5028.4
XS Rating Curve= 0 ,0
Exp/Cntr=0.3,0.1

Type RM Length L Ch R = 1 ,64484   ,1295,1295,1295
BEGIN DESCRIPTION:
ALLIGATOR BRANCH 35.0
END DESCRIPTION:
XS GIS Cut Line= 3
      3674055.07     10533457.78      3673946.56      10532144.8
      3672286.42     10531645.67
#Sta/Elev= 30
  3987.9  299.47  4065.8  296.96  4203.8  287.49  4359.7  277.25  4537.4  259.69
  4711.5  246.58  4798.2  242.81  4958.8  240.14  4964.3  239.93  4978.9  238.85
  4988.6  235.83    5019  239.54  5369.6   238.6  5565.3  239.15  5754.9  239.36
  5918.3  239.41  5931.5  236.75  5959.4  239.34  6140.2  242.51  6193.7  245.75
  6380.8  258.26  6414.8  265.06  6429.9  264.97  6440.4  268.29  6480.9  273.07
    6597  281.17  6689.5  291.19  6936.4   291.1  6983.4  289.13  7038.9  291.05
#Mann= 10 ,-1 , 0
  3987.9     .16       0  4203.8     .05       0  4711.5     .16       0
  4958.8     .07       0    5019     .12       0  5369.6     .16       0
  5565.3     .12       0  5754.9     .16       0  6193.7     .12       0
  6380.8     .16       0
Bank Sta=4964.3,5019
XS Rating Curve= 0 ,0
Exp/Cntr=0.3,0.1

Type RM Length L Ch R = 1 ,63189   ,710,710,710
BEGIN DESCRIPTION:
ALLIGATOR BRANCH 34.0
END DESCRIPTION:
XS GIS Cut Line= 3
      3675899.59     10532910.17      3674349.61     10531510.19
       3671928.3     10531493.76
#Sta/Elev= 30
  2932.9  300.48  3329.3  278.76  3421.2  276.38  3466.2  272.35  3513.2  266.65
  3655.4  258.07    3818   251.3    3910  250.88  3924.2  250.84  3945.1  243.82
  3966.7  249.64  3980.9  250.85  4193.2  251.73  4270.9  247.34    4448  243.08
  4561.6  243.76  4993.5  237.99  5000.2  237.87  5007.5  234.28  5014.4  235.06
  5041.5  238.05  5521.6  234.99  5915.2   237.7  6221.6  237.23  6461.6  246.92
  6811.6  272.93  6981.6  273.56  7161.6  283.53  7251.6  284.96  7442.9  297.82
#Mann= 8 ,-1 , 0
  2932.9     .16       0  3466.2     .05       0  3655.4     .16       0
    3910     .16       0  4993.5     .07       0  5014.4     .16       0
  5915.2     .16       0  6461.6     .16       0
#XS Ineff= 2 ,-1
 3476.14 4689.77  253.93 5886.36 6632.95  247.82
Permanent Ineff=
       F       F
Bank Sta=4993.5,5041.5
XS Rating Curve= 0 ,0
Exp/Cntr=0.3,0.1

Type RM Length L Ch R = 1 ,62479   ,497,497,497
BEGIN DESCRIPTION:
ALLIGATOR BRANCH 33.0
END DESCRIPTION:
XS GIS Cut Line= 3
      3676420.53     10533056.27      3674228.68     10530940.37
      3672004.44     10531244.17
#Sta/Elev= 30
  2124.9   314.8  2441.1  296.65  2745.1  283.25  2766.2  280.28  2815.9  281.02
    2837  277.27  2858.3  280.99  2971.5  284.14  3124.1  276.25  3183.5  268.86
  3335.9  256.91  3409.9  251.94    3620  249.73  3713.9   247.4  3735.3  249.34
  3777.7  245.74  3791.9  248.02  4633.4  238.24  4965.7     237  4979.9  234.77
  5015.4  237.75  5917.1  233.39  6199.9  237.19  6603.7   236.1  6736.6  241.11
  6866.1  248.91  7037.6  265.76  7209.2  291.73  7269.8   296.5  7416.3  299.16
#Mann= 8 ,-1 , 0
  2124.9     .16       0  3124.1     .05       0  3335.9      .1       0
    3620     .05       0  3735.3     .16       0  4965.7     .07       0
  4979.9     .16       0  6736.6     .16       0
#XS Ineff= 2 ,-1
 3817.05 4907.95  246.78 6015.91 6967.05  249.79
Permanent Ineff=
       F       F
Bank Sta=4965.7,5015.4
XS Rating Curve= 0 ,0
Exp/Cntr=0.3,0.1

Type RM Length L Ch R = 1 ,61982   ,1038,1038,1038
BEGIN DESCRIPTION:
ALLIGATOR BRANCH 32.0
END DESCRIPTION:
XS GIS Cut Line= 3
      3675799.61     10532210.19      3674399.61     10530660.19
      3671999.58     10531060.19
#Sta/Elev= 30
  2944.3   263.8  3043.8  257.99  3142.7   252.1  3305.6  247.28  3524.6  247.31
  3673.3  244.96  3709.1  242.71  3737.5  243.96  3978.2  240.29  4459.4  237.16
  4926.5  236.69  4969.1  235.26  4981.7     235  5182.5  236.59  5309.2  233.97
  5874.2  233.35  6221.6  234.01  6290.1  236.79  6421.9  237.46  6604.3  234.89
  6817.2  236.35  6908.5  242.33  7121.4  263.49  7293.7  284.99  7311.5  285.11
  7324.1  286.91  7334.3  290.71  7377.4  296.33  7415.4  297.84  7466.1  296.71
#Mann= 6 ,-1 , 0
  2944.3     .05       0  3043.8      .1       0  3305.6     .16       0
  4969.1     .07       0  4981.7     .16       0  7121.4     .16       0
#XS Ineff= 2 ,-1
 3550.49 4392.45246.9876 5756.82 7185.23  249.89
Permanent Ineff=
       F       F
Bank Sta=4459.4,5182.5
XS Rating Curve= 0 ,0
Exp/Cntr=0.3,0.1

Type RM Length L Ch R = 1 ,60944   ,669,669,669
BEGIN DESCRIPTION:
ALLIGATOR BRANCH 31.0
END DESCRIPTION:
XS GIS Cut Line= 4
      3676963.08     10532340.14      3674654.02     10529614.42
      3672292.91     10527392.19      3671234.27     10524910.45
#Sta/Elev= 30
  1843.6  312.37  1892.7  312.83  2087.4  312.81  2286.2  295.47  2782.8  249.11
  3293.6  238.32    3811  233.66  4414.1  232.64  4428.4   232.3    5981  235.09
  6454.7  237.68  6766.3   231.9  7445.2  233.56  7798.6  228.84  7989.9  233.46
    8273  233.42    8294  229.94  8364.8   234.1  8707.2  236.43  8899.7  232.16
  9562.8  231.91 10203.7  248.87 10238.2  244.45 10514.3  276.48 10628.3  285.58
 10719.5  285.22 10895.1  286.27 11095.5  290.62 11253.5  308.78 11356.4  307.98
#Mann= 7 ,-1 , 0
  1843.6     .05       0  1892.7     .16       0  2286.2     .16       0
  4414.1     .07       0  4428.4     .16       0 10719.5     .16       0
 10895.1     .05       0
#XS Ineff= 2 ,-1
 2495.45 3743.18  254.17 6436.3610588.64248.1564
Permanent Ineff=
       F       F
Bank Sta=3811,5981
XS Rating Curve= 0 ,0
Exp/Cntr=0.3,0.1

Type RM Length L Ch R = 1 ,60275   ,1759,1759,1759
BEGIN DESCRIPTION:
ALLIGATOR BRANCH 30.0
END DESCRIPTION:
XS GIS Cut Line= 4
       3676899.6     10531910.18      3675299.61     10529510.19
        3672989.     10527199.58       3671894.1     10524789.12
#Sta/Elev= 30
  2103.7  302.01  2626.8  249.97  2730.2     242  2868.4  238.28  2946.5  240.24
  3126.8  237.07  3337.1  230.59  3733.7  230.24  4079.2  233.82  4403.5  229.58
  4418.8  230.45  4656.1  233.37  5200.3  230.41  5737.7  232.84  7590.3  230.34
  7632.7  233.02  9320.5  232.93  9463.3  235.03  9606.1  246.89  9736.9   262.5
  9857.8  287.95  9981.7  283.76 10099.5  274.94 10133.6  269.52 10222.4  272.86
 10323.6  281.67 10429.8  298.96 10496.1  304.27 10686.2  309.76 10903.3  310.84
#Mann= 8 ,-1 , 0
  2103.7     .16       0  2626.8     .05       0  2730.2     .16       0
  4403.5     .07       0  4418.8     .16       0  9606.1     .05       0
  9981.7     .16       0 10222.4     .05       0
#XS Ineff= 2 ,-1
 2170.45 4034.09  248.29 6119.32 9670.45246.2866
Permanent Ineff=
       F       F
Bank Sta=4079.2,5737.7
XS Rating Curve= 0 ,0
Exp/Cntr=0.3,0.1

Type RM Length L Ch R = 1 ,58516   ,652,652,652
BEGIN DESCRIPTION:
ALLIGATOR BRANCH 29.0
END DESCRIPTION:
XS GIS Cut Line= 4
      3676949.62     10531810.23      3676349.61     10529610.19
      3675341.85     10528602.43      3674609.54      10524397.2
#Sta/Elev= 30
  2705.2  303.49  2922.9  278.96  3337.5  238.29    3937  228.51  4000.9  230.86
  4291.1  231.82  4626.3  229.51  4840.5  228.85  5607.8   231.6  6803.3  232.64
  7783.4  229.84  7864.6  235.99  7905.1  229.37  7976.2  228.99  7996.5  229.08
  8024.3  237.23  8047.3  237.83  8083.9   231.5  8169.1  231.66  8290.6  227.88
  8382.3  230.43  8783.8  229.52  8869.5  232.09  9113.1  228.95  9316.1  229.38
  9662.6  234.43  9955.6  241.75 10087.5  250.56 10544.3  294.19 10679.3  294.71
#Mann= 4 ,-1 , 0
  2705.2     .16       0  4626.3     .05       0  4840.5     .16       0
  9955.6     .05       0
#XS Ineff= 2 ,-1
 3039.77 4232.95  246.66 8039.7710426.14  246.41
Permanent Ineff=
       F       F
Bank Sta=4291.1,5607.8
XS Rating Curve= 0 ,0
Exp/Cntr=0.3,0.1

Type RM Length L Ch R = 1 ,57864   ,424,424,424
BEGIN DESCRIPTION:
ALLIGATOR BRANCH 28.0
END DESCRIPTION:
XS GIS Cut Line= 3
       3678049.6     10531360.17      3676799.61     10529810.19
      3676199.41     10525015.02
#Sta/Elev= 30
  3012.4  308.89  3076.6  305.26  3126.7  297.74  3161.9   283.2  3182.7  279.58
  3360.3  267.39  3368.2  263.86    3397   266.1  3403.4  263.35  3545.8  260.18
  3900.9  236.42  4171.1  233.23    4371  229.16  4385.4   229.6    5084  227.27
    5830  231.93  6182.7  228.65  6706.8  232.57  6847.9  228.88  7109.9  230.51
  7261.1  229.71  7291.3  236.95  7341.7  231.26  7523.1  228.44  8037.1  230.82
    8541  227.87  8772.8  240.84  9145.4   262.2  9522.4  279.02  9836.2  297.06
#Mann= 5 ,-1 , 0
  3012.4     .16       0    4371     .05       0  4385.4     .16       0
  8772.8     .05       0  9522.4     .16       0
#XS Ineff= 2 ,-1
 3608.52  4173.3  248.16 7307.39 9343.75  244.91
Permanent Ineff=
       F       F
Bank Sta=4171.1,7109.9
XS Rating Curve= 0 ,0
Exp/Cntr=0.3,0.1

Type RM Length L Ch R = 1 ,57440   ,1837,1837,1837
BEGIN DESCRIPTION:
ALLIGATOR BRANCH 27.0
END DESCRIPTION:
XS GIS Cut Line= 3
      3678119.93     10531036.95      3677219.35     10529865.11
       3676329.6     10525090.83
#Sta/Elev= 30
  3406.2  293.85  3511.4     297  3596.5  292.57  3660.9  293.69  4046.4  255.81
  4188.3  242.62  4360.5  233.55  4581.2  227.95  5184.6  229.24  5377.4  231.85
  5597.9  228.11  5704.4  228.07  5924.5  227.98    6025  228.15  6125.5  228.39
  6326.6  228.31  6597.9  229.01    6604  228.85  7116.8  229.17  7150.2  232.91
  7157.5   236.1  7238.9  229.44  8436.2  227.43    8439  226.93  8442.2  227.43
  8672.1  238.75    9167  274.17  9303.7  279.69  9476.8  294.96  9740.6  297.13
#Mann= 15 ,-1 , 0
  3406.2     .16       0  4046.4     .05       0  4581.2     .12       0
  5184.6     .05       0  5597.9     .12       0  5704.4     .05       0
  5924.5     .12       0    6025     .05       0  6125.5     .07       0
  6326.6     .05       0  6597.9     .07       0    6604     .05       0
  8436.2     .07       0  8442.2     .05       0  9303.7     .16       0
Bank Sta=4360.5,7150.2
XS Rating Curve= 0 ,0
Exp/Cntr=0.3,0.1

Type RM Length L Ch R = 1 ,55603   ,506,506,506
BEGIN DESCRIPTION:
ALLIGATOR BRANCH 26.0
END DESCRIPTION:
XS GIS Cut Line= 4
      3678054.85      10530765.7      3677653.38       10528856.
      3677197.65      10528215.8      3676481.78     10525504.19
#Sta/Elev= 30
  2653.9  306.11  2749.3  302.68  2966.1  274.77  3017.2  270.12  3137.9  264.86
  3194.7  258.66    3437  237.07  3670.9  232.84  3875.5  227.94  3926.6  230.01
  3957.3  228.05  5338.6  227.88  5351.9  227.93  5758.1  231.11  5935.9  229.32
  5956.1  233.44  5976.2  236.02  5991.2  235.17  6017.5  229.77  6038.2  228.72
  6462.8  228.79  6624.1  229.73  7275.9  227.28  7278.6  226.78  7281.9  227.28
  7404.9  232.13  7641.3  246.01    7948  274.91  8113.9  282.29  8195.7  289.54
#Mann= 12 ,-1 , 0
  2653.9     .16       0  3194.7     .05       0  3926.6     .05       0
  5338.6     .07       0  5351.9     .05       0  5758.1     .16       0
  5935.9     .05       0  6462.8     .12       0  6624.1     .05       0
  7275.9     .07       0  7281.9     .05       0  8113.9     .16       0
Bank Sta=3670.9,5956.1
XS Rating Curve= 0 ,0
Exp/Cntr=0.3,0.1

Type RM Length L Ch R = 1 ,55097   ,442,442,442
BEGIN DESCRIPTION:
ALLIGATOR BRANCH 25.0
END DESCRIPTION:
XS GIS Cut Line= 3
      3678250.17     10530841.71      3677599.13     10527195.84
      3676644.42     10525535.96
#Sta/Elev= 30
  2757.7  303.91  3165.6  278.86    3302  281.05  3360.9  277.51  3469.1  263.27
  3612.5  247.47    3753  241.31  4018.9  233.62  4161.1  228.04  4214.2  227.94
  4232.2  230.87  4252.5  227.92    5441  227.85  5542.6  230.08  5657.5  229.65
  5732.3  230.32  6226.5  229.53  6688.3  229.95  7021.7  228.59  7153.2  230.03
    7327  226.72  7329.7  226.22    7333  226.72  7549.9  230.28    7754  239.96
  8096.8  270.81  8193.8  289.43  8236.9  292.59  8252.7  296.17  8376.1  295.19
#Mann= 13 ,-1 , 0
  2757.7     .16       0  3469.1     .05       0    3753     .12       0
  4018.9     .05       0  5542.6     .12       0  5657.5     .05       0
  5732.3     .12       0  6226.5     .05       0  6688.3     .12       0
  7021.7     .05       0    7327     .07       0    7333     .05       0
  8096.8     .16       0
Bank Sta=4018.9,5542.6
XS Rating Curve= 0 ,0
Exp/Cntr=0.3,0.1

Type RM Length L Ch R = 1 ,54655   ,1411,1411,1411
BEGIN DESCRIPTION:
ALLIGATOR BRANCH 24.0
END DESCRIPTION:
XS GIS Cut Line= 3
      3678640.79     10530798.24        3678044.       10527402.
      3676655.11     10525427.17
#Sta/Elev= 30
  2676.7  296.23  2898.1  291.52    3176  279.27  3294.7  271.92  3446.4  257.91
  3629.1  243.81  3761.1  241.37  3813.6   238.6  4014.9  232.48  4025.1  232.48
  4207.9  227.86  5507.5  229.69  5639.5   228.9  5852.1  228.77  6094.2  228.68
    6890  229.85  7261.2   226.5  7263.9     226  7267.2   226.5  7435.3  227.27
  7586.1  231.27  7872.1   248.8  7966.8  255.89  8103.6  272.85  8124.5  272.79
  8154.1  278.72  8210.8  283.97  8225.6  290.83  8261.3   296.3  8539.3  295.74
#Mann= 12 ,-1 , 0
  2676.7     .05       0  3446.4     .12       0  3761.1     .07       0
  3813.6     .12       0  4025.1     .05       0  5507.5     .05       0
  5639.5     .12       0  5852.1     .16       0  6094.2     .05       0
  7261.2     .03       0  7267.2     .05       0  7872.1     .16       0
Bank Sta=4014.9,5507.5
XS Rating Curve= 0 ,0
Exp/Cntr=0.3,0.1

Type RM Length L Ch R = 1 ,53244   ,842,842,842
BEGIN DESCRIPTION:
ALLIGATOR BRANCH 23.0
END DESCRIPTION:
XS GIS Cut Line= 3
      3679458.21     10531376.99      3679443.74     10528693.24
      3676849.63     10525610.21
#Sta/Elev= 30
  2131.9  286.41  2658.7  274.26  2958.7  258.42  3028.7  261.65  3118.7  252.46
  3428.7  246.93  3468.7  243.71  3618.7  244.29  4048.7  234.69  4406.5  230.84
  4588.7  227.96  4638.7  231.99  4690.1  229.56  4941.2  230.47  4955.5  227.51
  6517.5  228.92  6605.8  226.94    7333  229.48  7678.5  226.18  7681.3  225.68
  7684.5  226.18  7684.6  226.19  7733.1  226.72  7923.6  228.71  7931.1  228.74
  8120.7  233.43  8439.8  252.67  8589.4  266.26  8780.6  292.66  8844.9   296.2
#Mann= 13 ,-1 , 0
  2131.9     .05       0  4406.5     .12       0  4690.1     .05       0
  4941.2     .07       0  6517.5     .16       0  6605.8     .05       0
  7678.5     .03       0  7684.5     .05       0  7684.6     .16       0
  7733.1     .05       0  7923.6     .16       0  7931.1     .05       0
  8120.7     .16       0
Bank Sta=4941.2,6517.5
XS Rating Curve= 0 ,0
Exp/Cntr=0.3,0.1

Type RM Length L Ch R = 1 ,52402   ,1139,1139,1139
BEGIN DESCRIPTION:
ALLIGATOR BRANCH 22.0
END DESCRIPTION:
XS GIS Cut Line= 3
      3680637.32     10531466.66       3679977.6     10528306.95
      3676899.59     10525410.17
#Sta/Elev= 30
  1583.5  319.24  2040.9  292.02  2203.1  277.51  2323.1  260.97  2475.6  250.02
  2670.5  245.18  3633.2  243.13  3817.1  232.95  4205.3  233.37  4399.4   228.2
  4634.9  230.38  4811.3  230.31  4913.8  228.68  4920.7  228.81  6307.2  227.78
  6439.6  228.34  6595.7  227.89  6697.2   228.3  6808.4  228.47  7262.5  228.97
  7535.4   224.6  7541.4   224.6  7870.8  229.22  8067.5  236.72  8238.8  241.79
  8544.8  258.96  8583.4  261.31  8698.4  269.46  8896.7  294.66  9038.1  296.56
#Mann= 18 ,-1 , 0
  1583.5     .16       0  2323.1     .05       0  3633.2     .07       0
  4205.3     .12       0  4399.4     .05       0  4634.9     .12       0
  4811.3     .07       0  4913.8     .07       0  6307.2     .12       0
  6439.6     .16       0  6595.7     .12       0  6697.2     .16       0
  6808.4     .12       0  7535.4     .03       0  7541.4     .12       0
  8067.5     .16       0  8544.8     .12       0  8583.4     .16       0
Bank Sta=4920.7,6307.2
XS Rating Curve= 0 ,0
Exp/Cntr=0.3,0.1

Type RM Length L Ch R = 1 ,51263   ,1279,1279,1279
BEGIN DESCRIPTION:
ALLIGATOR BRANCH 21.0
END DESCRIPTION:
XS GIS Cut Line= 3
      3682349.63     10530460.22      3680249.61     10527460.19
       3677549.6     10525060.18
#Sta/Elev= 30
  1305.2   296.8    1378  293.09  1678.8  264.31  2058.8  238.34  2202.9  233.24
  2497.6  234.01  2634.4  231.27  2798.4  233.53  2899.5  230.86  3136.2  231.51
  3316.3  228.28  3408.7  230.56    3754  227.07    4659  228.32  4665.1  228.01
  4995.2  226.13  6511.3   227.3  6610.8  226.92  6659.9  224.01    6681  226.13
    6901  228.16  7658.6  226.96  7772.3  230.33  7927.8  230.64  7935.4  231.56
  8034.1  237.66  8211.3  254.78  8317.5  267.29  8431.3  285.25  8579.7  285.85
#Mann= 4 ,-1 , 0
  1305.2     .16       0  2058.8     .05       0  4665.1     .07       0
  7935.4     .16       0
Bank Sta=4659,7927.8
XS Rating Curve= 0 ,0
Exp/Cntr=0.3,0.1

Type RM Length L Ch R = 1 ,49984   ,903,903,903
BEGIN DESCRIPTION:
ALLIGATOR BRANCH 20.0
END DESCRIPTION:
XS GIS Cut Line= 3
      3683749.61     10528910.19      3680845.65     10526883.34
      3677749.62      10524410.2
#Sta/Elev= 30
  1593.7  310.22  1946.6  287.81  2161.2  268.48    2319  265.32  2520.5  245.04
  2583.2  240.99  2828.5  229.51  2950.6  228.57  3022.1   225.6  3266.7  224.53
    3346  224.18  4889.8  225.53  4919.5  229.18  4925.6  228.35  4940.4  226.12
  4947.3  223.68  4996.9  223.01  5005.8  225.19  5553.7  224.97  5798.1  226.58
  7133.9  227.06  7731.1  224.63  7838.4  227.57  7923.2  226.59  8159.4  229.36
  8365.1  235.75  8677.3  248.85  8755.8  249.49  9017.9  279.46  9097.6   283.1
#Mann= 10 ,-1 , 0
  1593.7     .16       0  2583.2     .05       0  3266.7     .07       0
    3346     .05       0  4925.6     .07       0  5005.8     .05       0
  5553.7     .05       0  5798.1     .12       0  8159.4     .16       0
  9017.9     .12       0
Bank Sta=4940.4,5005.8
XS Rating Curve= 0 ,0
Exp/Cntr=0.3,0.1

Type RM Length L Ch R = 1 ,49081   ,685,685,685
BEGIN DESCRIPTION:
ALLIGATOR BRANCH 19.0
END DESCRIPTION:
XS GIS Cut Line= 3
      3683999.64     10528760.22      3681071.35      10526188.9
      3677999.65     10524260.21
#Sta/Elev= 30
   989.5  319.94  1074.5  314.54  1209.2  297.44  1391.8  285.49  1605.9  272.47
    1677  273.07  1789.9   262.2    1918  253.91  2107.4  245.48  2427.6  228.81
  2831.8  224.15  2874.5  226.44  2881.2  224.22  2888.8  225.55  2909.4  222.87
  2966.6  224.58  4730.6   225.8  4836.9  228.29  5003.5  223.88  5611.4  225.99
  6163.8  224.86  6265.2  227.51  6505.5  225.06  6867.2  226.68  6961.5  224.78
  7417.4  223.94  7641.3   225.8  8034.7  235.48  8128.9  240.47  8513.5  273.75
#Mann= 6 ,-1 , 0
   989.5     .16       0  1391.8      .1       0  2107.4     .05       0
  4836.9     .07       0  6265.2     .12       0  7641.3     .16       0
Bank Sta=4836.9,6265.2
XS Rating Curve= 0 ,0
Exp/Cntr=0.3,0.1

Type RM Length L Ch R = 1 ,48396   ,3073,3073,3073
BEGIN DESCRIPTION:
ALLIGATOR BRANCH 18.0
END DESCRIPTION:
XS GIS Cut Line= 3
      3684549.59     10528310.17      3680949.61     10525510.19
      3677949.59     10524010.18
#Sta/Elev= 30
   506.5  287.44   762.6  272.75   797.9   268.2     806  260.99   841.3  260.99
   848.5  267.77     891  269.79  1069.3  274.72  1098.3  279.83  1218.6  269.55
  1326.3  277.28  1487.2  254.91  1648.5   238.1  2010.4  228.18  2551.6  222.67
  3364.2  227.31    3813  224.01  4682.6  227.81  4981.2  223.92  5000.8  222.12
  5003.6  221.62  5006.8  222.12  5089.5  223.92  5483.2  224.12    7179   226.6
  7388.2  227.76    7485   228.3  7839.9  234.03  8256.4  281.16  8421.3  274.22
#Mann= 10 ,-1 , 0
   506.5     .16       0     891     .05       0  1487.2      .1       0
  1648.5     .05       0  5000.8     .03       0  5006.8     .07       0
  5483.2     .12       0    7179     .05       0  7388.2     .12       0
    7485     .16       0
Bank Sta=4981.2,5089.5
XS Rating Curve= 0 ,0
Exp/Cntr=0.3,0.1

Type RM Length L Ch R = 1 ,45323   ,940,940,940
BEGIN DESCRIPTION:
ALLIGATOR BRANCH 17.0
END DESCRIPTION:
XS GIS Cut Line= 3
      3684999.61     10528360.19      3680499.61     10523360.19
      3679299.63     10521960.21
#Sta/Elev= 30
 -1709.3  296.13 -1362.1   301.3 -1008.6  276.44  -725.3  276.24  -654.3  270.48
  -569.1  255.37  -335.9  242.42   160.4  228.22   648.5  223.15  2142.6  225.37
  2375.2  222.96  2460.2   222.8  2517.4  223.83  3700.2  225.86  3813.8  230.24
  4429.7   225.8  5017.5  222.42  5329.8  224.79  5951.4  222.93  6442.7  223.06
  6534.9  230.51  6585.6  239.88    6592  243.45  6598.6  241.79  6627.1  248.92
  6684.2  270.12  6690.8  268.71    6727  281.84  6776.4  288.02  6861.4  292.08
#Mann= 9 ,-1 , 0
 -1709.3     .05       0   648.5     .05       0  2375.2     .12       0
  2460.2     .07       0  2517.4     .12       0  4429.7     .05       0
  5329.8     .12       0  5951.4     .05       0  6585.6     .16       0
Bank Sta=4429.7,5329.8
XS Rating Curve= 0 ,0
Exp/Cntr=0.3,0.1

Type RM Length L Ch R = 1 ,44383   ,1399,1399,1399
BEGIN DESCRIPTION:
ALLIGATOR BRANCH 16.0
END DESCRIPTION:
XS GIS Cut Line= 3
      3684949.58     10526810.16      3680949.61     10522810.19
      3679349.62      10521610.2
#Sta/Elev= 30
  -644.7  285.64    -475  272.49  -390.2  257.31  -275.3  246.66   104.8  225.35
   734.7  222.87  1731.1  222.55  2028.1  225.59  2197.8  222.43  2914.3  223.13
  3371.3  222.73  4658.6  222.55  4785.8  226.48  4955.5   222.1  5008.3  218.56
  5054.8  223.15  5069.4  222.85  5269.4  220.81  5315.9  223.43  5453.6  222.98
  5640.6  223.34  5886.4  224.01  6340.2  224.11    6464  233.32  6612.1  253.48
  6640.2  259.75    6684  278.79  6775.7  297.76  6854.8  306.23  7012.1  302.61
#Mann= 12 ,-1 , 0
  -644.7     .16       0  -275.3     .05       0   734.7     .12       0
  2914.3     .05       0  3371.3     .12       0  4955.5     .07       0
  5069.4     .12       0  5315.9     .05       0  5453.6     .07       0
  5640.6     .12       0  5886.4     .05       0    6464     .16       0
Bank Sta=4955.5,5054.8
XS Rating Curve= 0 ,0
Exp/Cntr=0.3,0.1

Type RM Length L Ch R = 1 ,42984   ,4197,4197,4197
BEGIN DESCRIPTION:
ALLIGATOR BRANCH 15.0
END DESCRIPTION:
XS GIS Cut Line= 3
       3686049.6     10524910.18      3682049.61     10522110.19
      3679896.04     10521259.23
#Sta/Elev= 30
   135.4  317.75   198.9  315.66   315.4  311.19   330.3  304.43   357.3  309.34
   538.2  303.95   839.4  270.15  1119.3  254.17  1190.8  257.13  1318.4  247.94
  1410.3  242.05  1613.7  232.07    1863  226.17  3007.7  221.52  3675.3  222.07
  3703.6  217.68  3850.5  221.48  4802.2  224.05  4974.8  222.26  5032.9   220.6
  5050.3  222.55  5549.4   221.8  5638.6  217.37  5711.7  221.68  6894.5  221.19
  6999.2  226.69    7061  237.87  7153.2  279.47  7243.7  292.76  7333.6  299.06
#Mann= 12 ,-1 , 0
   135.4     .16       0   198.9     .05       0  1318.4     .12       0
  1410.3     .16       0    1863     .12       0  3007.7     .05       0
  3850.5     .12       0  4802.2     .05       0  4974.8     .07       0
  5050.3     .05       0  6894.5     .07       0  6999.2     .16       0
Bank Sta=4974.8,5032.9
XS Rating Curve= 0 ,0
Exp/Cntr=0.3,0.1

Type RM Length L Ch R = 1 ,38787   ,4753,4753,4753
BEGIN DESCRIPTION:
ALLIGATOR BRANCH 14.0
END DESCRIPTION:
XS GIS Cut Line= 3
      3685399.61     10522960.19      3681469.35      10520293.5
      3680145.55     10520749.23
#Sta/Elev= 30
     359  286.79   552.4  270.94   733.6   267.5   941.5  248.58  1079.2  254.31
  1309.8  255.54  1589.1   238.6  1627.1  234.04  1654.2  238.13  1828.3  232.75
  2056.8  226.84  2734.4  221.97  3016.6  221.43  3049.6  216.16  3073.6   220.4
  3289.2  219.08    3355  222.82    4649  222.59  4693.6  217.49  4966.2  218.63
    5038  220.16  5113.7  219.19  5815.4     222  5869.7  227.95  5909.6  238.02
  5922.6  247.27  6008.6  280.64  6134.1  281.58  6341.5  301.19  6508.6  299.68
#Mann= 10 ,-1 , 0
     359     .16       0  1589.1     .05       0  1828.3     .16       0
  2056.8     .05       0  2734.4     .12       0    3355     .05       0
  4966.2     .07       0    5038     .12       0  5113.7     .05       0
  5815.4     .16       0
Bank Sta=4966.2,5038
XS Rating Curve= 0 ,0
Exp/Cntr=0.3,0.1
