--- RESACA CREEK.prj (project) ---

Proj Title=RESACA CREEK Base Level Engineering
Current Plan=p01
Default Exp/Contr=0.3,0.1
English Units
Geom File=g01
Flow File=f01
Plan File=p01
Y Axis Title=Elevation
X Axis Title(PF)=Main Channel Distance
X Axis Title(XS)=Station
BEGIN DESCRIPTION:
RESACA CREEK
END DESCRIPTION:
DSS Export Rating Curves= 0
DSS Export Rating Curve Sorted= 0
DSS Export Volume Flow Curves= 0
DXF OffsetX= 0
DXF OffsetY= 0
DXF ScaleX= 1
DXF ScaleY= 10

--- RESACA CREEK.p01 (plan) ---

Plan Title=Multiple Run
Short Identifier=Multiple
Geom File=g01
Flow File=f01
Subcritical Flow
K Sum by GR= 0
Std Step Tol= 0.01
Critical Tol= 0.01
Num of Std Step Trials= 20
Max Error Tol= 0.3
Flow Tol Ratio= 0.001
Split Flow NTrial= 30
Split Flow Tol= 0.02
Split Flow Ratio= 0.02
Log Output Level= 0
Friction Slope Method= 1
Unsteady Friction Slope Method= 2
Unsteady Bridges Friction Slope Method= 1
Parabolic Critical Depth
Global Vel Dist=  1 , 1 , 1
Global Log Level= 0
CheckData=True
Encroach Param= -1, 0, 0, 0
BEGIN DESCRIPTION:
Multiple Run
END DESCRIPTION:

--- RESACA CREEK.f01 (steady flow) ---

Flow Title=Multiple
Program Version=4.10
Number of Profiles= 7
Profile Names=10-year,25-year,50-year,1pct_min,100-year,1pct_plu,500-year
River Rch & RM=RESACA CREEK,Reach-1         ,33008
     731    1023    1273    1165    1575    2131    2424
River Rch & RM=RESACA CREEK,Reach-1         ,32150
    1125    1605    2022    1871    2530    3422    3981
River Rch & RM=RESACA CREEK,Reach-1         ,28361
    1374    1967    2484    2301    3112    4208    4906
River Rch & RM=RESACA CREEK,Reach-1         ,20374
    1515    2172    2744    2541    3437    4648    5420
River Rch & RM=RESACA CREEK,Reach-1         ,13812
    1607    2303    2908    2690    3638    4920    5725
River Rch & RM=RESACA CREEK,Reach-1         ,7699
    2391    3483    4448    4156    5621    7602    9025
River Rch & RM=RESACA CREEK,Reach-1         ,7362
    2391    3483    4448    4156    5621    7602    9025
River Rch & RM=RESACA CREEK,Reach-1         ,4256
    2512    3660    4672    4364    5902    7981    9467
Boundary for River Rch & Prof#=RESACA CREEK,Reach-1         , 1
Up Type= 0
Dn Type= 3
Dn Slope=0.003
Boundary for River Rch & Prof#=RESACA CREEK,Reach-1         , 2
Up Type= 0
Dn Type= 3
Dn Slope=0.003
Boundary for River Rch & Prof#=RESACA CREEK,Reach-1         , 3
Up Type= 0
Dn Type= 3
Dn Slope=0.003
Boundary for River Rch & Prof#=RESACA CREEK,Reach-1         , 4
Up Type= 0
Dn Type= 3
Dn Slope=0.003
Boundary for River Rch & Prof#=RESACA CREEK,Reach-1         , 5
Up Type= 0
Dn Type= 3
Dn Slope=0.003
Boundary for River Rch & Prof#=RESACA CREEK,Reach-1         , 6
Up Type= 0
Dn Type= 3
Dn Slope=0.003
Boundary for River Rch & Prof#=RESACA CREEK,Reach-1         , 7
Up Type= 0
Dn Type= 3
Dn Slope=0.003
DSS Import GetInterval= 0
DSS Import GetPeak= 0
DSS Import FillOption= 0

--- RESACA CREEK.g01 (geometry) ---

Geom Title=Existing Conditions
Program Version=4.10

River Reach=RESACA CREEK    ,Reach-1
Reach XY= 30
      3682717.65     10495344.21      3681804.75       10496175.
      3681456.75       10496832.        3681782.       10498804.
        3682333.       10499500.       3681812.5       10500975.
        3682163.       10501573.      3682324.75       10502528.
       3683285.5       10503632.        3683325.       10504339.
      3683961.75       10504993.      3684446.75       10506134.
      3684663.75       10506147.       3684691.5       10506690.
      3685152.75       10506954.      3685118.75       10507327.
       3685593.5       10507772.      3686156.25       10507736.
      3686625.75       10509008.      3687812.75       10509002.
       3688264.5       10508681.      3689026.25       10508710.
        3690477.       10509232.      3691371.25       10508929.
      3692132.25       10510001.       3692564.5       10510057.
      3693554.75       10511088.        3693463.       10511699.
        3694207.       10512911.        3694285.       10514266.

Type RM Length L Ch R = 1 ,33008   ,443,443,443
BEGIN DESCRIPTION:
RESACA CREEK 63.0
END DESCRIPTION:
XS GIS Cut Line= 3
      3682349.62     10495110.21      3682549.61     10495510.19
       3682849.6     10495660.19
#Sta/Elev= 30
  4515.2  374.02  4573.9  368.62  4620.9  360.17  4636.4  357.76  4694.1  349.17
  4730.4  340.59  4747.2  337.88  4752.8  333.82  4769.5  332.28  4775.1  330.08
    4786  329.45  4805.9  327.39  4814.3  325.56  4828.2  324.82  4881.3  325.37
  4914.7  324.43  4917.4  323.93  4920.7  324.43  4984.8  325.43  4998.7  324.63
  5008.1   325.5  5021.1  327.05  5029.5  328.71  5051.8  329.41  5088.2  335.53
  5118.9  338.33  5141.3  342.11  5222.3  352.39  5267.1  356.53  5297.8  362.12
#Mann= 7 ,-1 , 0
  4515.2     .16       0  4620.9     .12       0  4636.4     .16       0
    4786     .12       0  4914.7     .07       0  4920.7     .12       0
  5008.1     .16       0
Bank Sta=4805.9,5021.1
XS Rating Curve= 0 ,0
Exp/Cntr=0.3,0.1

Type RM Length L Ch R = 1 ,32565   ,415,415,415
BEGIN DESCRIPTION:
RESACA CREEK 62.0
END DESCRIPTION:
XS GIS Cut Line= 3
      3681949.64     10495610.21      3682349.61     10495860.19
      3682449.62     10496260.22
#Sta/Elev= 30
  4563.8  347.55  4650.4  339.04    4687  333.08  4702.3  325.93  4708.2  328.54
  4712.5  326.48  4717.1  324.27  4729.4  324.75  4738.9  327.94  4752.4  325.23
  4811.4  325.15  4830.2  320.93    4833  320.43  4836.2  320.93  4890.1  322.32
  4912.2  322.23  4927.6   324.3  5012.5  323.27    5030  325.19    5038  326.71
  5046.5  324.25  5094.7  326.04  5107.6  323.65    5136   326.8  5141.1  324.95
  5157.2  326.22  5164.8  326.47  5218.4  329.42  5285.8  338.88  5447.8   361.9
#Mann= 9 ,-1 , 0
  4563.8     .16       0  4712.5     .05       0  4830.2     .07       0
  4836.2     .05       0  4890.1     .12       0  5046.5     .05       0
  5157.2     .16       0  5164.8     .05       0  5285.8     .16       0
Bank Sta=4811.4,5030
XS Rating Curve= 0 ,0
Exp/Cntr=0.3,0.1

Type RM Length L Ch R = 1 ,32150   ,481,481,481
BEGIN DESCRIPTION:
RESACA CREEK 61.0
END DESCRIPTION:
XS GIS Cut Line= 3
      3681649.62      10495660.2      3681999.61     10496060.19
      3682399.61     10496310.19
#Sta/Elev= 30
  4441.6  376.16  4477.2   373.1  4534.1  361.96  4597.7   353.9  4675.5  340.47
  4746.7  330.37  4760.5  329.52  4767.6  326.33  4780.4  325.28    4817  321.02
  4838.8  318.18  4942.1  318.04  4944.8  317.54  4948.1  318.04  5096.3  318.14
  5117.6  320.96  5152.7  326.31  5292.6     344  5306.2  346.53  5315.1  346.12
  5327.5  349.16  5336.9  349.14  5342.8  347.17  5358.1  347.37  5379.3   352.5
  5385.8  357.34  5406.4  358.68  5415.9  359.84  5421.8  361.98  5444.8  364.19
#Mann= 7 ,-1 , 0
  4441.6     .16       0  4780.4     .12       0  4942.1     .07       0
  4948.1     .12       0  5152.7     .16       0  5292.6     .05       0
  5406.4     .16       0
Bank Sta=4817,5117.6
XS Rating Curve= 0 ,0
Exp/Cntr=0.3,0.1

Type RM Length L Ch R = 1 ,31669   ,254,254,254
BEGIN DESCRIPTION:
RESACA CREEK 60.0
END DESCRIPTION:
XS GIS Cut Line= 3
      3681549.62     10496060.21      3681749.61     10496360.19
      3682149.58     10496710.16
#Sta/Elev= 30
  4606.1  353.24  4634.6  351.67  4700.7  343.48  4706.7  341.59  4721.8  339.85
  4727.8  337.21  4750.3  334.39  4793.9  324.53  4808.9  323.26  4835.6  318.61
  4836.9   318.4    4863  315.62  4865.7  315.12    4869  315.62  5118.7  315.62
  5157.9  316.05  5179.2  317.79  5186.3  319.99  5207.2  321.41  5214.8   323.3
  5243.3  326.73  5249.9  326.51  5257.5  328.88  5278.4  331.05  5327.8  339.39
    5342  340.51  5363.8  344.86    5399  348.05  5413.2   351.2  5498.1  362.02
#Mann= 6 ,-1 , 0
  4606.1     .16       0  4835.6     .12       0  4836.9     .07       0
    4863     .07       0    4869     .07       0  5118.7     .16       0
Bank Sta=4836.9,5179.2
XS Rating Curve= 0 ,0
Exp/Cntr=0.3,0.1

Type RM Length L Ch R = 1 ,31415   ,614,614,614
BEGIN DESCRIPTION:
RESACA CREEK 59.0
END DESCRIPTION:
XS GIS Cut Line= 3
      3680507.89       10496861.      3681302.14     10496470.39
      3682148.49     10496782.89
#Sta/Elev= 30
  3744.6  383.71    3783     382  3889.8   384.8  3924.8  382.08  4075.1  361.42
  4120.1  353.74  4136.6  353.85  4187.5  346.85  4193.1  347.73    4210  343.75
  4215.5  345.06  4232.4  340.73    4238  342.01  4299.9  333.08  4371.5   326.2
  4440.3  318.24  4457.2  316.24  4531.5  316.62    4589  315.62  4591.8  315.12
    4595  315.62  4801.7  315.62  4830.3  315.62  4910.3  316.49  5121.2  315.79
  5149.3  317.88  5194.7  324.56  5298.6  335.38  5383.9  349.88  5531.9  365.34
#Mann= 9 ,-1 , 0
  3744.6     .16       0  4371.5     .12       0  4531.5     .07       0
    4589     .07       0    4595     .07       0  4801.7     .16       0
  4830.3     .05       0  4910.3     .07       0  5121.2     .16       0
Bank Sta=4440.3,5149.3
XS Rating Curve= 0 ,0
Exp/Cntr=0.3,0.1

Type RM Length L Ch R = 1 ,30801   ,98,98,98
BEGIN DESCRIPTION:
RESACA CREEK 58.0
END DESCRIPTION:
XS GIS Cut Line= 3
      3681149.61     10497410.19      3681549.61     10497110.19
      3681949.61     10496810.19
#Sta/Elev= 30
  4499.4  364.08  4521.3  359.68  4549.4  358.07  4556.7  353.63  4562.9   352.2
  4606.7  343.96  4642.1  339.22  4656.7  333.48  4677.5  330.76  4685.9  331.12
  4706.7  325.78  4712.9  326.32  4806.7  316.52  4811.1  316.21  4865.4  315.62
  5098.2  315.62  5121.3  315.62 5126.14  317.43  5142.1  317.72  5182.9  311.14
  5185.6  310.64  5188.9  311.14  5277.5  325.02  5321.3  328.22  5327.5  330.32
  5371.3  334.32  5377.5  336.28  5399.4  337.91  5427.5  342.32  5499.4  347.31
#Mann= 6 ,-1 , 0
  4499.4     .16       0  4811.1     .12       0  4865.4     .05       0
  5098.2     .16       0  5182.9    .033       0  5188.9     .16       0
Bank Sta=4806.7,5126.14
XS Rating Curve= 0 ,0
Exp/Cntr=0.3,0.1

Type RM Length L Ch R = 1 ,30703   ,63,63,63
BEGIN DESCRIPTION:
Mapping XS 6f3b69fe
END DESCRIPTION:
XS GIS Cut Line= 5
      3681055.75     10497487.16      3681177.25     10497445.94
      3681613.44     10497185.52      3681672.04     10497146.46
      3682009.56     10496854.37
#Sta/Elev= 30
  4385.8  371.89  4427.5  370.83  4487.7  366.49  4614.5  342.87  4630.1  337.55
  4672.9   334.1  4731.2  323.55  4826.6  316.85  4847.9  319.55  4912.8  316.19
  4921.9  318.95  4927.8  315.62  4943.3  318.62  4949.2  315.62  4994.4  315.62
  5001.7  318.86  5044.2  318.18  5065.6  316.68  5074.2  312.36  5080.2  314.96
  5109.5  311.07  5172.9  311.96  5208.4  312.39  5212.8  308.88  5215.6  308.38
  5218.8  308.88  5230.1  313.48  5272.9  315.15    5365  324.34  5538.9  350.48
#Mann= 6 ,-1 , 0
  4385.8     .05       0  4427.5     .16       0  4847.9     .12       0
  5172.9     .16       0  5212.8     .07       0  5218.8     .16       0
Bank Sta=5001.7,5044.2
XS Rating Curve= 0 ,0
Exp/Cntr=0.3,0.1

Type RM Length L Ch R = 1 ,30640   ,353,353,353
BEGIN DESCRIPTION:
Mapping XS 535422a1
END DESCRIPTION:
XS GIS Cut Line= 4
      3681064.44      10497534.9      3681465.87     10497376.49
      3681852.16      10497070.5      3682138.64     10496849.13
#Sta/Elev= 30
  4371.1  371.21  4473.4  366.85  4527.2  359.45  4538.5  355.86  4573.9  349.67
  4587.3  344.31  4602.4  341.85  4641.4  339.03  4665.8  333.68  4742.2  324.46
  4785.2  316.27  4844.3  311.56  4916.7  309.27  4966.3  310.34  4977.8  305.28
  4980.5  304.78  4983.8  305.28  5001.6  308.22  5009.6  307.51    5016  310.01
  5044.9  308.39  5073.7  310.74    5165  311.38  5201.9   309.8  5298.7  313.84
  5365.6  320.13  5415.5   326.9  5436.3  331.47  5457.1  332.89  5657.5  364.42
#Mann= 6 ,-1 , 0
  4371.1     .05       0  4573.9     .16       0  4844.3     .12       0
  4977.8     .07       0  4983.8     .12       0  5298.7     .16       0
Bank Sta=4966.3,5016
XS Rating Curve= 0 ,0
Exp/Cntr=0.3,0.1

Type RM Length L Ch R = 1 ,30287   ,462,462,462
BEGIN DESCRIPTION:
RESACA CREEK 57.0
END DESCRIPTION:
XS GIS Cut Line= 3
      3681299.56     10497560.19      3681649.61     10497560.19
      3682049.59     10497160.21
#Sta/Elev= 30
  4667.4  349.13  4677.4  348.15  4697.4  344.03  4717.4  340.82  4747.4  337.97
  4753.3  336.58  4757.4  335.61  4787.4   332.5  4847.4  321.56  4857.4  318.75
  4867.4  317.68  4877.4   315.6  4947.4  309.27    4962  308.74  4977.4  308.41
  4994.4  303.56  4997.2  303.06  5000.4  303.56  5014.9  307.51  5088.2  308.31
  5413.4  307.05  5427.6  307.24    5470  309.61  5484.1  310.99  5495.1  312.96
  5526.6   317.4  5540.7  320.55    5569  325.44  5579.6  328.56  5583.1  328.56
#Mann= 6 ,-1 , 0
  4667.4     .05       0  4753.3     .16       0    4962     .12       0
  4994.4     .07       0  5000.4     .12       0  5495.1     .16       0
Bank Sta=4977.4,5014.9
XS Rating Curve= 0 ,0
Exp/Cntr=0.3,0.1

Type RM Length L Ch R = 1 ,29825   ,496,496,496
BEGIN DESCRIPTION:
RESACA CREEK 56.0
END DESCRIPTION:
XS GIS Cut Line= 4
      3681003.46     10497856.46      3681437.48      10498012.7
      3682210.05      10497882.5      3682583.28     10497491.91
#Sta/Elev= 30
    4304  358.21  4328.1  355.09  4414.9  354.73  4608.1  344.14  4703.8  335.34
  4747.4  326.44  4889.1  310.69  4980.4  306.63  4993.3  305.43  4997.7  302.77
  5000.4  302.27  5003.7  302.77  5010.8  305.61    5163  310.49  5416.9  314.86
    5545  321.55  5613.7  327.51  5627.9  325.43  5670.3  325.82  5684.5   326.9
  5698.6  331.23  5804.6   328.2  5882.6  333.54  5889.5   328.8  5896.9  335.52
  5946.2   341.6  5953.1  339.62  5967.2  344.06  5995.5  347.02    6089  351.03
#Mann= 5 ,-1 , 0
    4304     .16       0  4997.7     .07       0  5003.7     .16       0
    5545     .05       0  5896.9     .16       0
Bank Sta=4889.1,5163
XS Rating Curve= 0 ,0
Exp/Cntr=0.3,0.1

Type RM Length L Ch R = 1 ,29329   ,417,417,417
BEGIN DESCRIPTION:
RESACA CREEK 55.0
END DESCRIPTION:
XS GIS Cut Line= 3
      3681399.65     10498460.19      3681749.61     10498460.19
      3682499.59     10498310.19
#Sta/Elev= 30
  4663.4  350.73  4703.4  344.78  4783.4   330.3  4873.4  317.09  4903.4  311.39
  4943.4  307.88  4993.4  303.31  5000.4  300.87  5003.1  300.37  5006.4  300.87
  5010.9  303.72    5044  303.59  5094.9  305.22  5135.7  307.91  5217.3  310.24
  5240.3  309.78  5339.7  306.58  5400.9  311.55  5492.7  310.96  5516.4  312.52
  5533.5  314.85  5543.7  312.31  5553.9  312.56  5564.1  314.92  5594.7  316.18
    5615  318.46    5666  326.11  5737.4  329.14  5757.8  333.64  5778.2  333.95
#Mann= 5 ,-1 , 0
  4663.4     .16       0  5000.4     .07       0  5006.4     .16       0
  5240.3     .12       0  5516.4     .05       0
Bank Sta=4943.4,5135.7
XS Rating Curve= 0 ,0
Exp/Cntr=0.3,0.1

Type RM Length L Ch R = 1 ,28912   ,551,551,551
BEGIN DESCRIPTION:
RESACA CREEK 54.0
END DESCRIPTION:
XS GIS Cut Line= 3
       3681449.6     10498860.19      3681849.61     10498860.19
      3682549.57     10498360.22
#Sta/Elev= 30
  4633.2  331.34  4693.2  323.03  4703.2  320.59  4803.2  309.04  4843.2  305.56
  4913.2  302.37  4983.2   302.6  4993.2  301.41  5000.2  298.97    5003  298.47
  5006.2  298.97  5013.2  302.07  5124.7  301.41  5156.1  301.66  5168.4  303.07
  5191.7  302.42    5349  305.72  5463.3  306.27  5500.2   307.3  5535.8  310.17
  5547.3  308.99  5577.6  309.15  5586.2   311.2    5628  313.76  5684.5  319.55
  5758.3   325.1  5785.3  328.28  5814.8  333.68  5820.9  332.67  5893.4  335.49
#Mann= 5 ,-1 , 0
  4633.2     .16       0  5000.2     .07       0  5006.2     .16       0
  5124.7     .12       0  5547.3     .05       0
Bank Sta=4983.2,5013.2
XS Rating Curve= 0 ,0
Exp/Cntr=0.3,0.1

Type RM Length L Ch R = 1 ,28361   ,288,288,288
BEGIN DESCRIPTION:
RESACA CREEK 53.0
END DESCRIPTION:
XS GIS Cut Line= 4
      3681095.51     10499583.77      3681678.87     10499458.76
       3682338.6     10499229.59      3683218.86     10498924.62
#Sta/Elev= 30
  3914.4  352.51  4092.5  344.55  4235.6  328.92  4241.2  326.81  4442.2   310.9
  4482.2  308.64  4574.1  304.26  4675.1  300.69  4763.1   299.1  5006.1  299.52
  5117.5  298.28    5144  298.26  5146.7  297.76    5150  298.26  5223.6  300.71
  5263.4  301.75  5345.2   299.9  5411.6  300.69  5435.7  303.43  5499.7  305.92
  5647.8  309.33  5681.2  307.76  5769.2  309.85  5868.1  312.74    5966   320.6
  6038.7  328.03  6044.4  329.48  6049.7  328.11  6075.6  332.29    6141  336.05
#Mann= 16 ,-1 , 0
  3914.4     .05       0  4442.2     .16       0  4482.2     .08       0
  4574.1     .16       0  5006.1     .12       0  5117.5     .05       0
    5144     .07       0    5150     .05       0  5223.6     .08       0
  5345.2     .16       0  5435.7     .08       0  5499.7     .16       0
  5647.8     .08       0  5769.2     .05       0    5966     .08       0
  6038.7     .05       0
Bank Sta=4675.1,5223.6
XS Rating Curve= 0 ,0
Exp/Cntr=0.3,0.1

Type RM Length L Ch R = 1 ,28073   ,281,281,281
BEGIN DESCRIPTION:
RESACA CREEK 52.0
END DESCRIPTION:
XS GIS Cut Line= 4
      3681130.28     10499972.64       3682026.1     10499597.65
      3682442.76     10499444.87       3683316.2     10499112.13
#Sta/Elev= 30
  3708.6  353.83  3772.9  352.71  3933.6  344.15    4163  327.91  4390.8  303.39
    4534  298.69  4593.6  297.07  4668.5  297.17  4695.8  297.09  4802.7  297.15
  4909.5  297.49    4925  297.49  4992.4   298.4  4999.1  296.15  5001.8  295.65
  5005.1  296.15  5007.4  298.46  5016.3  298.19  5123.1  297.02    5181  296.95
  5334.2  299.05  5431.1  305.74  5445.2  307.21  5483.2  310.86  5568.2  312.61
  5603.6  317.88  5790.9  321.14  5863.4  322.32  5931.4   324.8  6058.2  327.44
#Mann= 18 ,-1 , 0
  3708.6     .05       0  3933.6     .16       0  4593.6     .05       0
  4668.5     .16       0  4695.8     .07       0  4802.7     .12       0
  4909.5     .05       0    4925     .12       0  4999.1     .07       0
  5005.1     .12       0  5016.3     .05       0  5123.1     .12       0
    5181     .05       0  5431.1      .1       0  5445.2     .05       0
  5790.9     .08       0  5863.4     .05       0  5931.4     .08       0
Bank Sta=4534,5334.2
XS Rating Curve= 0 ,0
Exp/Cntr=0.3,0.1

Type RM Length L Ch R = 1 ,27792   ,689,689,689
BEGIN DESCRIPTION:
RESACA CREEK 51.0
END DESCRIPTION:
XS GIS Cut Line= 3
      3681237.82     10500035.28      3683017.34     10499453.68
      3683615.45     10498942.25
#Sta/Elev= 30
    3995  350.93  4003.8  350.65  4083.2  346.36  4199.3  341.04  4354.6  334.56
  4450.2  320.83  4659.7  297.49  4765.7  295.26    4790  295.36  4938.1  296.24
  5046.2  296.06  5130.1  294.86  5132.8  294.36  5136.1  294.86  5148.8  295.52
  5254.1  296.65  5374.6  296.16  5438.2  298.29  5576.4   306.3    5596  309.29
  5659.1  306.65  5799.5  312.42  5871.9  312.96    5885  315.09  5892.7  312.51
  5984.9  314.47  6292.1  324.04  6313.7  324.17  6458.2  328.13  6654.1  329.98
#Mann= 15 ,-1 , 0
    3995     .05       0  4003.8     .16       0  4083.2     .05       0
  4199.3     .16       0  4765.7     .05       0    4790     .16       0
  4938.1     .12       0  5046.2     .05       0  5130.1     .07       0
  5136.1     .05       0  5148.8     .12       0  5254.1     .05       0
  6292.1     .12       0  6313.7     .08       0  6458.2     .05       0
Bank Sta=4659.7,5438.2
XS Rating Curve= 0 ,0
Exp/Cntr=0.3,0.1

Type RM Length L Ch R = 1 ,27103   ,476,476,476
BEGIN DESCRIPTION:
RESACA CREEK 50.0
END DESCRIPTION:
XS GIS Cut Line= 3
      3681517.85     10500000.86      3681949.61     10500310.19
      3682749.58     10500810.17
#Sta/Elev= 30
  4484.7  335.46  4628.9  327.59  4664.5  322.52  4679.3  322.97  4750.5  311.84
  4765.3     312  4771.4  309.52    4807  304.82  4907.7  294.58  5026.4  290.99
  5029.1  290.49  5032.4  290.99  5038.8  292.65  5065.9  292.78  5196.8  292.59
  5227.5  294.29  5428.6  296.26  5554.9     305  5604.9   307.8  5610.8  305.72
  5626.1  307.78    5632  306.56  5647.3  309.13  5653.2  307.42  5711.6  315.28
  5757.3  318.55    5915  334.38  5930.3  337.41  5936.2  336.18  5959.2  338.86
#Mann= 6 ,-1 , 0
  4484.7     .16       0  5026.4     .07       0  5032.4     .16       0
  5065.9     .05       0  5554.9     .16       0  5757.3      .1       0
Bank Sta=4907.7,5227.5
XS Rating Curve= 0 ,0
Exp/Cntr=0.3,0.1

Type RM Length L Ch R = 1 ,26627   ,472,472,472
BEGIN DESCRIPTION:
RESACA CREEK 49.0
END DESCRIPTION:
XS GIS Cut Line= 3
      3681449.64     10500460.21      3681849.61     10500760.19
      3682649.63     10500860.19
#Sta/Elev= 30
  4527.9  331.19    4531  331.19  4535.1  328.53    4556  327.59  4605.1  319.13
  4620.6  318.28  4670.6  309.39    4706   306.2  4725.2  303.08  4835.1  290.54
  4864.3  291.59  4985.1  290.76  4996.7  289.39  4999.5  288.89  5002.7  289.39
    5006  290.41  5063.1  290.81    5179  290.12  5199.2  291.24  5259.6   290.8
  5320.1  291.96  5468.8  296.59  5554.4  301.38  5571.2  303.41    5635  308.47
  5642.6  310.38    5693  313.93  5703.1  315.83  5715.7  316.16  5834.1  329.27
#Mann= 7 ,-1 , 0
  4527.9     .05       0  4605.1      .1       0  4725.2     .16       0
  4996.7     .07       0  5002.7     .16       0  5063.1     .05       0
  5571.2      .1       0
Bank Sta=4985.1,5006
XS Rating Curve= 0 ,0
Exp/Cntr=0.3,0.1

Type RM Length L Ch R = 1 ,26155   ,451,451,451
BEGIN DESCRIPTION:
RESACA CREEK 48.0
END DESCRIPTION:
XS GIS Cut Line= 3
      3681499.63     10501310.18      3681899.61     10501160.19
       3682699.6     10501060.19
#Sta/Elev= 30
  4576.6  338.82  4652.2  327.27  4762.6  315.58  4768.8  313.56  4908.6  299.46
  4918.3  297.27  4933.5  296.69  4950.4  294.38  4963.7  288.47  4988.7  290.36
    4994  285.11  4998.1  285.02  5000.9  284.52  5004.1  285.02    5034  285.43
  5041.6  288.46  5078.9  288.82  5316.2  291.93  5385.9  295.96    5486  302.75
  5525.3  305.67  5530.3  307.29  5588.3  309.66  5605.9  313.75  5648.8  319.13
  5741.3  327.63  5743.5  327.79  5767.2  330.23  5772.2  329.41    5810  334.69
#Mann= 8 ,-1 , 0
  4576.6     .16       0  4998.1     .07       0  5004.1     .16       0
  5078.9     .05       0  5385.9     .16       0    5486      .1       0
  5741.3     .16       0  5743.5      .1       0
Bank Sta=4988.7,5041.6
XS Rating Curve= 0 ,0
Exp/Cntr=0.3,0.1

Type RM Length L Ch R = 1 ,25704   ,488,488,488
BEGIN DESCRIPTION:
RESACA CREEK 47.0
END DESCRIPTION:
XS GIS Cut Line= 3
      3681749.58      10501660.2      3682099.61     10501510.19
      3682499.58      10501410.2
#Sta/Elev= 30
  4587.3  328.25  4601.8  326.87  4609.1  324.86    4620  324.08  4630.9  321.12
  4641.7  320.23  4654.4  316.18  4663.5  315.98  4739.6  304.24    4794  298.15
  4830.3  295.43  4859.3  289.78  4877.5   287.4  4924.6  287.78  4935.5  286.41
  4959.1  287.78  4986.2  286.34  4988.3   282.7  4991.1   282.2  4994.3   282.7
    4999  283.06  5009.4  287.36  5068.6  289.97  5091.8  289.92  5138.6  292.51
  5174.3  295.02  5192.3  298.23  5241.5  301.52  5328.9  309.33  5380.4  312.14
#Mann= 5 ,-1 , 0
  4587.3     .16       0  4988.3     .07       0  4994.3     .16       0
  5138.6     .05       0  5241.5      .1       0
Bank Sta=4986.2,5009.4
XS Rating Curve= 0 ,0
Exp/Cntr=0.3,0.1

Type RM Length L Ch R = 1 ,25216   ,443,443,443
BEGIN DESCRIPTION:
RESACA CREEK 46.0
END DESCRIPTION:
XS GIS Cut Line= 3
      3681604.67     10502084.19      3682099.61     10501910.19
      3682499.59      10501510.2
#Sta/Elev= 30
    4482  332.32  4497.8  332.49  4506.1   331.2  4599.1  327.91    4661  327.48
  4699.2  325.58  4794.6  314.53  4805.2  314.46  4815.9  312.11  4826.4  311.61
  4858.2  306.71  4872.5  305.55  4879.4  303.69  4921.8  299.47  4953.6   294.1
  4974.8  288.56    5001  281.88  5003.7  281.38    5007  281.88  5010.2  281.88
  5020.8   285.5  5063.2   287.3  5105.6  286.26  5119.8  287.49  5162.2  287.21
  5224.8  288.54  5331.9  291.18  5430.9  298.47  5501.6  301.83  5572.3  308.13
#Mann= 4 ,-1 , 0
    4482     .16       0    5001     .07       0    5007     .16       0
  5224.8     .05       0
Bank Sta=4974.8,5020.8
XS Rating Curve= 0 ,0
Exp/Cntr=0.3,0.1

Type RM Length L Ch R = 1 ,24773   ,482,482,482
BEGIN DESCRIPTION:
RESACA CREEK 45.0
END DESCRIPTION:
XS GIS Cut Line= 3
      3682049.62     10502510.18      3682249.61     10502310.19
      3682649.59     10502010.21
#Sta/Elev= 30
  4689.7  318.53  4693.2  318.53  4703.8  316.11  4746.3  308.97  4760.4  307.79
  4774.5  304.94  4802.8  302.41    4817   299.6  4885.4  293.61  4930.1  289.38
  4944.2  287.15  4958.4  282.16    4969  283.85  4986.1   283.2  4994.4  282.29
  4997.7  281.07  5000.4  280.57  5003.7  281.07  5015.2  283.44  5029.8  285.25
  5050.7  283.57  5077.6  285.47  5122.5  285.22  5165.2  286.89  5229.8   287.9
  5279.8  290.64  5379.8   294.2  5450.9  299.34    5459  300.47  5472.5  300.82
#Mann= 6 ,-1 , 0
  4689.7     .16       0  4885.4     .12       0  4997.7     .07       0
  5003.7     .12       0  5077.6     .05       0  5450.9      .1       0
Bank Sta=4986.1,5015.2
XS Rating Curve= 0 ,0
Exp/Cntr=0.3,0.1

Type RM Length L Ch R = 1 ,24291   ,591,591,591
BEGIN DESCRIPTION:
RESACA CREEK 44.0
END DESCRIPTION:
XS GIS Cut Line= 3
      3682099.59     10502660.19      3682499.61     10502660.19
      3682849.59     10502260.21
#Sta/Elev= 30
  4589.2  315.95  4649.2  307.04  4679.2  301.44  4759.2  291.85  4769.2  289.69
  4832.9  286.46  4939.2  283.32  4956.2  279.21    4959  278.71  4962.2  279.21
  4969.2  282.83  4989.3  280.72  4992.5  280.72    5003  279.33  5010.6  281.24
  5017.2  281.28  5081.8  281.28  5095.5  285.07  5116.9  286.46    5131  286.04
  5188.1  287.67  5194.7  286.91  5263.8  289.77  5308.1  291.95  5356.2  296.12
  5414.4  299.86  5442.4  302.99    5450  302.57    5507  307.22  5520.7  307.34
#Mann= 8 ,-1 , 0
  4589.2     .16       0  4832.9      .1       0  4956.2     .07       0
  4962.2      .1       0  4989.3     .16       0    5131      .1       0
  5263.8     .05       0  5356.2      .1       0
Bank Sta=4992.5,5017.2
XS Rating Curve= 0 ,0
Exp/Cntr=0.3,0.1

Type RM Length L Ch R = 1 ,23700   ,501,501,501
BEGIN DESCRIPTION:
RESACA CREEK 43.0
END DESCRIPTION:
XS GIS Cut Line= 3
      3682399.61     10503360.19      3682749.61     10502960.19
      3683149.59     10502860.19
#Sta/Elev= 30
  4462.2   313.2  4547.1  306.58  4554.7   301.8  4561.4  304.28  4575.6  294.02
  4589.9  295.65  4596.5  299.77  4604.1  291.83  4607.3  292.08    4625  291.56
  4646.8  296.82  4702.8  294.77  4724.6  289.18  4781.1  289.17  4794.9  286.29
  4924.9  280.87  4979.9  280.81  4986.6  280.06  4990.4  276.13  5011.7  279.44
  5065.9   281.4  5091.2  275.76    5094  275.26  5097.2  275.76  5107.1  282.21
  5126.1  280.52  5148.3  280.21    5272  290.58  5382.8  306.23    5406   307.3
#Mann= 6 ,-1 , 0
  4462.2     .16       0  4607.3      .1       0  4924.9     .16       0
  5091.2     .07       0  5097.2     .16       0  5126.1      .1       0
Bank Sta=4979.9,5011.7
XS Rating Curve= 0 ,0
Exp/Cntr=0.3,0.1

Type RM Length L Ch R = 1 ,23199   ,712,712,712
BEGIN DESCRIPTION:
RESACA CREEK 42.0
END DESCRIPTION:
XS GIS Cut Line= 3
      3682599.63     10503460.18      3682999.61     10503260.19
       3683149.6      10503110.2
#Sta/Elev= 30
  4582.1   306.5    4596  304.01  4649.2  298.62  4663.1  295.82  4679.9  295.19
  4685.5  293.19  4738.6  288.46    4747   288.7  4752.6  287.25  4836.4  283.19
  4850.4   281.8  4872.8  281.72  4886.7  280.25  4903.5  280.52  4909.1  279.41
  4948.2  278.83  4976.2     280  4992.9  278.81  4995.5  273.61  4998.3  273.11
  5001.5  273.61  5006.9  277.35  5043.4  278.25  5071.7  277.16    5088   278.9
  5114.1   280.6  5128.3  281.96  5142.4  284.51  5170.7   286.5  5241.4  296.32
#Mann= 4 ,-1 , 0
  4582.1     .16       0  4995.5     .07       0  5001.5     .16       0
    5088      .1       0
Bank Sta=4992.9,5006.9
XS Rating Curve= 0 ,0
Exp/Cntr=0.3,0.1

Type RM Length L Ch R = 1 ,22487   ,492,492,492
BEGIN DESCRIPTION:
RESACA CREEK 41.0
END DESCRIPTION:
XS GIS Cut Line= 3
       3682849.6     10503710.19      3683249.61     10503610.19
      3683449.63     10503560.18
#Sta/Elev= 30
  4610.1  292.87  4651.3  288.91  4661.7  288.67  4669.4  286.97  4682.3  286.46
  4710.6  283.16  4723.5  282.42  4733.8  280.65  4785.3  278.67  4793.1  277.26
  4880.7  276.85    4940  277.54  4950.3  277.24    4958  275.35  4991.5   275.3
  4996.2  269.39    4999  268.89  5002.2  269.39  5004.4  271.41  5012.1  275.02
  5019.8  276.61  5040.5  275.12  5063.7  280.58  5081.7  283.26  5094.6  284.96
  5128.1  287.04  5146.1  290.57  5156.4  291.13  5205.4  299.15  5228.6  302.13
#Mann= 3 ,-1 , 0
  4610.1     .16       0  4996.2     .07       0  5002.2     .16       0
Bank Sta=4991.5,5012.1
XS Rating Curve= 0 ,0
Exp/Cntr=0.3,0.1

Type RM Length L Ch R = 1 ,21995   ,595,595,595
BEGIN DESCRIPTION:
RESACA CREEK 40.0
END DESCRIPTION:
XS GIS Cut Line= 3
      3682849.61     10504360.19      3683249.61     10503960.19
      3683599.63     10503960.19
#Sta/Elev= 30
  4444.3  307.34  4585.7  294.41    4614  292.48  4628.1  290.28  4642.3  289.75
  4656.4   287.9  4684.7  285.29  4769.6  278.93  4783.7  277.06  4854.4   274.6
  4953.4  275.79  4981.7  275.61  4992.8  267.57  4995.6  267.07  4998.8  267.57
  5006.4  274.69    5020   274.8    5030  272.41    5040  275.17    5070  276.01
    5080  277.18    5090  277.56    5100  279.07    5120  280.96    5140  282.24
    5150  283.56    5200  287.54    5270  294.64    5280  294.91    5360  303.79
#Mann= 3 ,-1 , 0
  4444.3     .16       0  4992.8     .07       0  4998.8     .16       0
Bank Sta=4981.7,5006.4
XS Rating Curve= 0 ,0
Exp/Cntr=0.3,0.1

Type RM Length L Ch R = 1 ,21400   ,475,475,475
BEGIN DESCRIPTION:
RESACA CREEK 39.0
END DESCRIPTION:
XS GIS Cut Line= 3
      3683099.64     10504610.17      3683399.61     10504360.19
      3683799.63     10504210.18
#Sta/Elev= 30
  4579.2  303.61  4707.4  291.87  4771.2  284.87  4799.8   283.3  4841.5  279.23
  4933.9  273.67  4972.3  273.89  4979.5  271.84  4984.8  273.28    4991  269.29
  4998.7  267.44  5001.5  266.94  5004.7  267.44  5009.7   271.2  5015.1  273.35
  5055.1  272.67  5095.2  275.43  5100.5  277.88  5108.5  277.22  5119.2  274.59
  5130.8  275.66  5140.6  278.12  5161.9  281.12    5258  290.59  5301.6  299.34
  5321.2  300.88  5351.5  306.21  5356.8  305.65  5381.7  308.83  5396.9  309.34
#Mann= 3 ,-1 , 0
  4579.2     .16       0  4998.7     .07       0  5004.7     .16       0
Bank Sta=4984.8,5015.1
XS Rating Curve= 0 ,0
Exp/Cntr=0.3,0.1

Type RM Length L Ch R = 1 ,20925   ,551,551,551
BEGIN DESCRIPTION:
RESACA CREEK 38.0
END DESCRIPTION:
XS GIS Cut Line= 3
      3683399.61     10504910.19      3683699.61     10504660.19
       3683849.6     10504360.21
#Sta/Elev= 30
  4575.4  303.96  4589.1  304.02  4625.5  300.56  4660.7  294.81  4681.5  292.62
  4689.3  290.58  4710.1  289.18  4717.9  287.26  4724.4  287.36  4753.1   281.9
  4767.4  280.94  4825.1  272.94  4831.2  271.85  4845.5  271.39  4888.2  272.06
  4979.9   271.7  4999.3  262.73    5002  262.23  5005.3  262.73  5010.6  270.91
  5069.3  276.53  5077.7  276.24  5153.2  284.64  5211.9   292.8  5242.6  298.62
  5256.6  299.75  5270.6  303.07  5287.3  305.12  5298.5  308.31  5301.3  308.31
#Mann= 5 ,-1 , 0
  4575.4     .16       0  4825.1     .12       0  4888.2     .16       0
  4999.3     .07       0  5005.3     .16       0
Bank Sta=4979.9,5010.6
XS Rating Curve= 0 ,0
Exp/Cntr=0.3,0.1

Type RM Length L Ch R = 1 ,20374   ,550,550,550
BEGIN DESCRIPTION:
RESACA CREEK 37.0
END DESCRIPTION:
XS GIS Cut Line= 3
      3683449.58      10505160.2      3683849.61     10504960.19
      3684249.59     10504560.21
#Sta/Elev= 30
  4602.6  312.11  4736.8  295.56  4812.3  282.25  4879.3   273.5  4943.9  270.22
  4974.4  270.62  4993.7  261.85  4996.5  261.35  4999.7  261.85  5005.1  267.96
  5041.5  267.54    5047  264.16  5053.4  264.16  5078.1  270.53  5219.5  272.19
  5264.3  269.27  5276.1  266.38  5332.7  271.42    5361   266.4  5375.1  272.57
  5389.3  274.04  5403.4  269.13  5445.8  273.72    5460  269.01  5488.2  275.08
  5530.7  275.91  5570.7   288.8  5573.7  289.65  5601.4  299.25  5615.5  299.18
#Mann= 7 ,-1 , 0
  4602.6     .16       0  4943.9     .12       0  4993.7     .07       0
  4999.7     .12       0  5264.3     .16       0  5570.7     .05       0
  5573.7     .08       0
Bank Sta=4974.4,5005.1
XS Rating Curve= 0 ,0
Exp/Cntr=0.3,0.1

Type RM Length L Ch R = 1 ,19824   ,519,519,519
BEGIN DESCRIPTION:
RESACA CREEK 36.0
END DESCRIPTION:
XS GIS Cut Line= 3
      3683749.58     10505710.22      3684099.61     10505310.19
      3684399.64     10505160.17
#Sta/Elev= 30
  4477.7  305.37  4499.1  302.84  4505.7  300.93  4574.2  292.66  4591.2  289.75
  4597.8  289.92  4649.8  283.91  4740.2  275.05  4768.7  270.77  4810.4  267.86
  4867.4  266.58  4881.6  267.71  4981.3   269.2  4987.9  266.64  4995.5  261.62
  4999.1  260.96  5001.9  260.46  5005.1  260.96  5005.9  264.69  5017.6  263.47
  5023.2  265.93  5031.6   265.6    5040  267.73  5062.4  268.63    5115  268.11
    5135  268.41  5165.8  273.15  5267.3  285.65  5305.3  290.32  5344.7  295.14
#Mann= 8 ,-1 , 0
  4477.7     .12       0  4574.2     .16       0  4649.8     .12       0
  4999.1     .07       0  5005.1     .12       0    5115     .16       0
  5267.3     .12       0  5305.3     .16       0
Bank Sta=4981.3,5005.9
XS Rating Curve= 0 ,0
Exp/Cntr=0.3,0.1

Type RM Length L Ch R = 1 ,19305   ,464,464,464
BEGIN DESCRIPTION:
RESACA CREEK 35.0
END DESCRIPTION:
XS GIS Cut Line= 3
       3683849.6     10505810.19      3684249.61     10505660.19
      3684549.56      10505610.2
#Sta/Elev= 30
  4598.3   306.2  4613.4  303.68  4638.4  301.52  4651.7  298.47  4683.7  295.62
  4754.1  285.69    4779  283.27  4784.3  283.69  4790.5  282.16  4819.6  279.79
  4864.4  274.71    4876   271.7  4918.7  265.54  4930.3  264.89  4940.1  266.04
  4985.5  266.59  4993.5  264.33  5001.1  259.02  5003.9  258.52  5007.1  259.02
  5015.7   266.5  5096.5  266.71  5115.5  268.38  5119.3  267.83  5126.9  270.38
  5147.2  273.69  5180.1  277.22  5187.7     279  5218.1  281.53  5329.6  298.83
#Mann= 5 ,-1 , 0
  4598.3     .16       0  4819.6     .12       0  5001.1     .07       0
  5007.1     .12       0  5115.5     .16       0
Bank Sta=4985.5,5015.7
XS Rating Curve= 0 ,0
Exp/Cntr=0.3,0.1

Type RM Length L Ch R = 1 ,18841   ,762,762,762
BEGIN DESCRIPTION:
RESACA CREEK 34.0
END DESCRIPTION:
XS GIS Cut Line= 3
      3684049.59     10506360.21      3684449.61     10506010.19
      3684599.62     10505760.17
#Sta/Elev= 30
  4516.9  298.04  4521.4  297.61  4531.9  295.99    4581  290.96  4626.7  284.25
  4687.3  276.17  4743.3  271.37  4800.2  270.22  4807.8  268.93  4828.7  269.37
    4843  267.39  4882.8  266.63  4928.4  265.81  4949.3  263.49  4977.7  264.83
  4984.4  264.05    4992   257.7  4995.6  257.58  4998.4  257.08  5001.6  257.58
  5006.2  260.92  5012.8  261.05  5020.4  264.92  5045.2  265.36    5099  264.71
  5114.5  265.78  5151.4   271.4  5157.3  273.97    5237  286.64    5340  298.63
#Mann= 8 ,-1 , 0
  4516.9     .12       0  4521.4     .16       0  4531.9     .12       0
  4626.7     .16       0  4882.8     .12       0  4995.6     .07       0
  5001.6     .12       0  5045.2     .16       0
Bank Sta=4977.7,5020.4
XS Rating Curve= 0 ,0
Exp/Cntr=0.3,0.1

Type RM Length L Ch R = 1 ,18079   ,474,474,474
BEGIN DESCRIPTION:
RESACA CREEK 33.0
END DESCRIPTION:
XS GIS Cut Line= 3
      3683952.22     10506621.99      3684768.22     10506318.16
      3684863.48     10505763.91
#Sta/Elev= 30
  4224.2  308.74  4301.2   306.6  4326.2  303.61  4331.6  305.07  4344.4  303.54
  4356.6  301.61  4417.2  299.35  4434.8  296.98  4442.2  294.36  4447.6  295.59
  4488.2  285.65  4520.2  279.83  4527.9  277.04  4613.6  266.47  4699.2  262.46
  4754.6  263.45  4854.8  262.76  4936.6  263.28    4979  262.01    5008  254.13
  5010.8  253.63    5014  254.13  5016.9  259.64  5022.3  260.95  5079.9  262.15
  5214.6  267.99  5359.8  280.88  5545.1  295.49  5550.2  294.53  5657.3  298.17
#Mann= 7 ,-1 , 0
  4224.2     .12       0  4344.4     .16       0  4854.8     .12       0
    5008     .07       0    5014     .12       0  5079.9     .16       0
  5359.8     .12       0
Bank Sta=4979,5022.3
XS Rating Curve= 0 ,0
Exp/Cntr=0.3,0.1

Type RM Length L Ch R = 1 ,17605   ,435,435,435
BEGIN DESCRIPTION:
RESACA CREEK 32.0
END DESCRIPTION:
XS GIS Cut Line= 3
      3684373.84     10507067.21      3684677.68       10506937.
      3685094.33     10506077.65
#Sta/Elev= 30
  4440.5  294.49    4475  294.48  4492.2  294.28  4595.8   293.3  4624.8  290.84
  4695.5  289.04    4701  286.98  4724.6  286.09  4800.9  279.71  4813.7  277.03
  4823.1  276.99  4966.2  260.18  4978.7   260.6  4988.7  257.31  4994.3  257.29
  4997.9  252.21  5000.7  251.71  5003.9  252.21  5011.3  256.97  5016.9  257.57
  5023.1  260.32  5045.4  259.44  5131.3  260.56  5287.8  259.25  5361.9  260.03
  5428.8  260.23  5547.2  273.66  5586.8  280.26  5662.1  288.03  5726.1  291.77
#Mann= 9 ,-1 , 0
  4440.5     .16       0    4475     .12       0  4492.2     .16       0
  4595.8     .12       0  4724.6     .16       0  4997.9     .07       0
  5003.9     .16       0  5131.3     .12       0  5361.9     .16       0
Bank Sta=4978.7,5023.1
XS Rating Curve= 0 ,0
Exp/Cntr=0.3,0.1

Type RM Length L Ch R = 1 ,17170   ,558,558,558
BEGIN DESCRIPTION:
RESACA CREEK 31.0
END DESCRIPTION:
XS GIS Cut Line= 4
      3684477.98     10507084.56      3684729.76     10507101.93
      3685163.79     10506884.91      3685632.56     10506450.87
#Sta/Elev= 30
  4339.2  292.21  4380.9  291.84  4441.1  295.09  4481.2  294.25  4595.2  282.34
  4646.5  275.66  4652.1  276.21  4680.9  272.26  4719.2  269.37  4803.1  258.42
  4852.5  257.28  4937.2  259.09  4949.2  257.42  4971.5  257.57  4987.5  256.06
  4990.9  252.62  4993.7  252.12  4996.9  252.62  5004.3  255.85  5009.9  253.34
  5016.3  258.58  5105.2  257.38  5328.4  258.08  5381.7  259.92    5431   266.1
  5544.4  276.48  5593.7  284.25  5664.6  291.46  5671.4  293.26  5715.7  295.86
#Mann= 7 ,-1 , 0
  4339.2     .16       0  4595.2     .12       0  4852.5     .16       0
  4990.9     .07       0  4996.9     .16       0  5105.2     .12       0
  5328.4     .16       0
Bank Sta=4971.5,5016.3
XS Rating Curve= 0 ,0
Exp/Cntr=0.3,0.1

Type RM Length L Ch R = 1 ,16612   ,444,444,444
BEGIN DESCRIPTION:
RESACA CREEK 30.0
END DESCRIPTION:
XS GIS Cut Line= 3
      3684749.59      10507660.2      3685149.61     10507360.19
      3685799.61     10506560.19
#Sta/Elev= 30
  4497.5   290.1  4504.7  289.76  4553.4  284.52  4590.2  279.83  4660.2  274.41
    4808  260.49  4815.7  259.86  4904.8  255.41    4984  256.99  4990.2  254.21
  4991.4  250.04  4994.1  249.54  4997.4  250.04  5000.7  250.04  5004.7  253.69
  5019.1  256.67  5203.7   255.3  5332.3  257.64  5405.3   256.1  5474.3  254.54
  5495.3   256.3  5573.6  255.96  5611.7  257.69  5765.4  268.59  5878.9  271.87
  5957.2  276.06  5985.9  278.67  5992.4  282.47  6014.7  282.46  6028.3   280.1
#Mann= 10 ,-1 , 0
  4497.5     .07       0  4504.7     .16       0  4553.4     .05       0
  4660.2     .16       0    4808     .05       0  4815.7     .16       0
  4991.4     .07       0  4997.4     .16       0  5405.3     .12       0
  5611.7     .16       0
Bank Sta=4984,5019.1
XS Rating Curve= 0 ,0
Exp/Cntr=0.3,0.1

Type RM Length L Ch R = 1 ,16168   ,443,443,443
BEGIN DESCRIPTION:
RESACA CREEK 29.0
END DESCRIPTION:
XS GIS Cut Line= 3
      3685098.06     10508010.88      3685449.61     10507610.19
      3686199.58     10506810.21
#Sta/Elev= 30
    4474  283.88  4532.1  282.11  4595.7  276.86  4620.9  273.45  4661.2  270.75
  4666.9  269.17  4716.2  266.18  4752.3  261.81  4787.4   259.9  4909.5  255.22
  4913.6  255.15  4985.7  254.78  4993.3  253.21  4996.9  248.71  4999.7  248.21
  5002.9  248.71  5003.7  251.58  5010.5  251.58  5014.1  255.32  5324.7  253.36
  5365.7  253.12  5430.1  253.36  5516.4  253.52  5544.6  254.07  5636.9  262.39
  5672.1  263.71  5813.7  260.81  5919.7  269.98  6040.3  286.01  6103.6   293.6
#Mann= 13 ,-1 , 0
    4474     .12       0  4620.9     .16       0  4661.2     .05       0
  4787.4     .12       0  4909.5     .05       0  4913.6     .16       0
  4996.9     .07       0  5002.9     .16       0  5324.7     .12       0
  5365.7     .05       0  5430.1     .07       0  5516.4     .05       0
  6040.3      .1       0
Bank Sta=4985.7,5014.1
XS Rating Curve= 0 ,0
Exp/Cntr=0.3,0.1

Type RM Length L Ch R = 1 ,15725   ,532,532,532
BEGIN DESCRIPTION:
RESACA CREEK 28.0
END DESCRIPTION:
XS GIS Cut Line= 3
      3685599.61     10508060.19      3685799.61     10507810.19
      3686599.57     10507060.22
#Sta/Elev= 30
  4678.2  283.09  4774.1  271.15    4792   269.4  4927.1  254.97  4976.8  254.16
  4995.2  247.49  5002.4   247.1  5005.2   246.6  5008.4   247.1  5012.3  249.94
  5019.6  248.83  5026.5  253.82  5048.5  253.11    5069  252.72  5076.3  248.14
  5090.4  247.17  5097.3  253.49  5118.8  252.45  5158.1  254.82  5196.4  257.26
  5245.8  253.66  5330.8  252.74  5338.1  254.94  5380.6   257.9  5423.1   254.8
  5472.8  256.39  5769.4  271.45  5868.5  274.78  5984.7   285.7  6094.9  294.84
#Mann= 10 ,-1 , 0
  4678.2     .16       0  4774.1     .05       0    4792     .16       0
  5002.4     .07       0  5008.4     .16       0  5048.5     .12       0
  5158.1     .07       0  5245.8     .05       0  5472.8      .1       0
  5984.7     .07       0
Bank Sta=4976.8,5026.5
XS Rating Curve= 0 ,0
Exp/Cntr=0.3,0.1

Type RM Length L Ch R = 1 ,15193   ,367,367,367
BEGIN DESCRIPTION:
RESACA CREEK 27.0
END DESCRIPTION:
XS GIS Cut Line= 3
      3685599.63     10508110.18      3686252.59     10507793.85
      3686823.64      10507404.5
#Sta/Elev= 30
    4354     287  4385.1  284.63  4398.4  281.49  4428.4  278.57  4509.5  268.01
  4587.3  260.55  4624.1  255.39  4652.3  252.62  4966.2  251.97  4974.5   251.3
  4988.8  250.55  4995.5  247.71  4998.2  247.21  5001.5  247.71  5020.7  251.76
  5056.6  253.61  5073.6  256.13    5078  255.52  5109.4   260.8  5124.4  260.81
  5130.4  262.65  5151.4  263.53  5303.9  278.07  5345.9  279.21  5366.8  280.29
  5375.7  282.03  5421.7  284.03  5591.2  297.32    5642  300.05  5770.7     303
#Mann= 8 ,-1 , 0
    4354     .16       0  4428.4     .05       0  4624.1     .16       0
  4652.3     .05       0  4974.5      .1       0  4995.5     .07       0
  5001.5      .1       0  5421.7     .05       0
Bank Sta=4966.2,5020.7
XS Rating Curve= 0 ,0
Exp/Cntr=0.3,0.1

Type RM Length L Ch R = 1 ,14826   ,449,449,449
BEGIN DESCRIPTION:
RESACA CREEK 26.0
END DESCRIPTION:
XS GIS Cut Line= 3
      3685549.61     10508160.19      3686249.61     10508160.19
      3686549.58      10508060.2
#Sta/Elev= 30
  4280.9  292.47  4310.9  293.35  4320.9  290.25  4370.9  285.79  4410.9  280.93
  4430.9  278.31  4450.9  273.49  4493.6  269.25  4500.9  269.16  4510.9  266.47
  4530.9  263.45  4580.9   259.1  4630.9  252.05  4670.9  250.86  4790.2  250.48
  4890.9  251.62  4900.9  250.63  4951.1  251.06  4970.9  250.86  4983.5  249.65
  4991.4  245.84    4999  244.44  5001.7  243.94    5005  244.44  5012.5  251.63
  5086.3  258.11  5117.9  262.33  5181.2     269    5255  278.77  5297.1  283.04
#Mann= 6 ,-1 , 0
  4280.9     .16       0  4493.6     .05       0  4790.2     .12       0
  4951.1     .16       0    4999     .07       0    5005     .16       0
Bank Sta=4983.5,5012.5
XS Rating Curve= 0 ,0
Exp/Cntr=0.3,0.1

Type RM Length L Ch R = 1 ,14377   ,565,565,565
BEGIN DESCRIPTION:
RESACA CREEK 25.0
END DESCRIPTION:
XS GIS Cut Line= 3
      3685549.58     10508210.17      3686349.61     10508560.19
      3686749.57     10508260.22
#Sta/Elev= 30
  4145.7  293.89  4178.1  289.76  4200.3   289.1  4212.4   285.6    4244  282.33
    4306  273.05  4358.2   269.3  4381.6  265.83  4440.4  261.94  4462.7  258.83
  4509.4   256.2  4549.6  251.69  4655.2  249.17  4678.6  250.74  4713.3  248.72
  4806.5  248.63  4981.1  250.31  4994.1  244.29  4996.9  243.79  5000.1  244.29
  5016.2  249.03  5063.6  251.36  5082.5  252.77  5097.1  251.68  5105.4  254.49
  5111.7  253.04  5118.9  255.36  5140.8  258.06  5268.9  268.23  5518.9  293.72
#Mann= 5 ,-1 , 0
  4145.7     .16       0  4806.5     .12       0  4994.1     .07       0
  5000.1     .12       0  5063.6     .16       0
Bank Sta=4981.1,5016.2
XS Rating Curve= 0 ,0
Exp/Cntr=0.3,0.1

Type RM Length L Ch R = 1 ,13812   ,492,492,492
BEGIN DESCRIPTION:
RESACA CREEK 24.0
END DESCRIPTION:
XS GIS Cut Line= 3
      3686035.55     10509538.67      3686599.61     10508910.19
      3686899.62     10508510.18
#Sta/Elev= 30
  4169.9  281.57  4207.4  280.36  4228.4  277.54  4249.3  277.88  4256.8  275.92
    4271  275.87  4285.2  274.08  4320.3  272.55  4327.8  271.17  4433.2  265.81
    4561  261.93  4759.1  251.73  4858.5  250.41  4915.3  247.56  4922.1  244.84
  4929.5  245.29  4943.7   248.2  4966.4  248.37  4986.4  248.67  4997.6  242.12
  5000.3  241.62  5003.6  242.12  5017.5  242.77  5021.7  248.56  5121.7  247.84
  5157.1  249.58  5236.3  257.81  5286.3  261.28  5407.1  272.26  5514.4  283.13
#Mann= 5 ,-1 , 0
  4169.9     .16       0  4433.2     .12       0  4966.4     .16       0
  4997.6     .07       0  5003.6     .16       0
Bank Sta=4986.4,5021.7
XS Rating Curve= 0 ,0
Exp/Cntr=0.3,0.1

Type RM Length L Ch R = 1 ,13320   ,502,502,502
BEGIN DESCRIPTION:
RESACA CREEK 23.0
END DESCRIPTION:
XS GIS Cut Line= 3
      3686899.61     10509410.21      3686949.61     10509010.19
      3686899.62     10508610.24
#Sta/Elev= 30
  4680.9  260.99  4756.7  255.06    4822   250.8  4902.6  247.89  4965.6  247.19
  4983.3  242.54  4993.3  242.04  5003.4  245.73  5016.2  246.59  5023.6  247.15
  5041.2  246.68  5046.2  241.14  5050.8  241.01  5053.6  240.51  5056.8  241.01
  5063.9   245.8    5074  246.79  5094.1  247.14  5174.7  245.91  5235.2  247.19
  5295.7  252.61  5325.9  256.59  5356.1  259.37  5363.7  260.85  5368.7  260.65
  5396.4  263.27  5444.3  269.58  5456.9  270.13  5477.1  272.39  5487.1  274.17
#Mann= 5 ,-1 , 0
  4680.9     .16       0  4756.7     .12       0  5016.2     .16       0
  5050.8     .07       0  5056.8     .16       0
Bank Sta=4965.6,5003.4
XS Rating Curve= 0 ,0
Exp/Cntr=0.3,0.1

Type RM Length L Ch R = 1 ,12818   ,482,482,482
BEGIN DESCRIPTION:
RESACA CREEK 22.0
END DESCRIPTION:
XS GIS Cut Line= 3
      3687599.61     10509310.19      3687349.61     10508960.19
       3687449.6     10508560.22
#Sta/Elev= 30
    4558  267.87  4571.5  265.18  4580.1  261.39  4594.9  256.85  4607.2  254.96
  4636.7   254.9  4651.4  252.88  4724.7  249.07  4758.3  246.74  4838.2  244.38
  4888.6  244.13  4951.3  245.33  4956.9  240.07  4959.6  239.57  4962.9  240.07
  4964.3  241.75    4966  243.79  4974.6  242.11  4980.7  243.27  4998.4  243.27
  5011.3  240.45    5019  245.21  5122.1  253.47  5176.2  258.83    5184  260.68
  5217.5  263.86  5225.2  265.56  5294.8  273.94    5336  281.17  5400.4  289.57
#Mann= 5 ,-1 , 0
    4558     .16       0  4724.7     .12       0  4956.9     .07       0
  4962.9     .12       0  4964.3     .16       0
Bank Sta=4998.4,5019
XS Rating Curve= 0 ,0
Exp/Cntr=0.3,0.1

Type RM Length L Ch R = 1 ,12336   ,514,514,514
BEGIN DESCRIPTION:
RESACA CREEK 21.0
END DESCRIPTION:
XS GIS Cut Line= 3
      3687649.62     10509260.16      3687749.61     10509010.19
      3687499.62     10508610.21
#Sta/Elev= 30
  4726.4   257.3  4765.4  254.42  4780.2  254.59  4843.5   249.7    4897  247.31
  4974.1   243.9  4980.8  242.14  4986.2  243.28  4989.9  239.49  4992.7  238.99
  4995.9  239.49  5018.6  243.59    5031   244.5  5119.5  243.17  5176.6  245.23
  5249.8  253.91  5255.7  253.64  5301.6  259.16  5307.5  259.01    5314  260.75
  5328.8  261.81    5373  268.89  5380.7     271  5401.9  272.88  5408.4  275.26
  5423.1  276.72  5438.4  279.91  5459.7  281.37  5464.4  283.77  5467.3  283.77
#Mann= 5 ,-1 , 0
  4726.4     .16       0    4897     .12       0  4989.9     .07       0
  4995.9     .12       0  5119.5     .16       0
Bank Sta=4986.2,5018.6
XS Rating Curve= 0 ,0
Exp/Cntr=0.3,0.1

Type RM Length L Ch R = 1 ,11822   ,493,493,493
BEGIN DESCRIPTION:
RESACA CREEK 20.0
END DESCRIPTION:
XS GIS Cut Line= 3
      3688149.61     10509460.15      3688099.61     10508760.19
       3688249.6     10508410.22
#Sta/Elev= 30
  4279.4  279.04  4359.6  272.63  4369.6  270.85  4399.7  268.71  4479.9  260.07
    4520  257.43  4580.1  251.65  4700.4  243.96  4730.5   243.4  4740.5  242.27
  4777.9  242.23  4934.1  242.71  4990.2  241.48  4999.9  238.62  5002.7  238.12
  5005.9  238.62  5013.8  242.78  5048.2   242.7  5066.4  243.82  5100.8  244.36
  5133.5  247.48  5142.5  249.16  5155.2   249.8  5187.9  254.71  5200.6  255.22
  5218.7  259.09  5242.3  261.87  5300.3  270.63  5340.2  274.28  5361.9  275.28
#Mann= 5 ,-1 , 0
  4279.4     .16       0  4777.9     .12       0  4934.1     .16       0
  4999.9     .07       0  5005.9     .16       0
Bank Sta=4990.2,5013.8
XS Rating Curve= 0 ,0
Exp/Cntr=0.3,0.1

Type RM Length L Ch R = 1 ,11329   ,464,464,464
BEGIN DESCRIPTION:
RESACA CREEK 19.0
END DESCRIPTION:
XS GIS Cut Line= 3
       3688199.6     10509410.21      3688549.61     10508660.19
      3688649.61     10508360.18
#Sta/Elev= 30
  4195.3  275.84    4204  274.65  4232.4  273.87  4239.5  272.65  4255.2  272.59
  4294.6  268.88  4300.9  267.61  4316.7  267.04  4323.8  265.48    4375  262.57
  4382.9  261.28  4512.2  251.39  4654.9  245.86  4682.7  245.61  4700.6  244.51
  4758.1  245.76  4901.6  241.97  4980.2  240.88  4991.4  241.05  5000.9  238.11
  5011.3  237.87    5014  237.37  5017.3  237.87  5020.2  241.16  5086.2  246.75
  5117.8   250.4  5181.1  254.68  5265.4  265.07  5318.1  269.83  5339.2  273.26
#Mann= 5 ,-1 , 0
  4195.3     .16       0  4682.7     .12       0  4980.2     .16       0
  5011.3     .07       0  5017.3     .16       0
Bank Sta=4991.4,5020.2
XS Rating Curve= 0 ,0
Exp/Cntr=0.3,0.1
