HEC-RAS study WHEELOCK CREEK.prj: WHEELOCK CREEK Base Level Engineering

--- WHEELOCK CREEK.g01 (geometry) --- (continued)

Type RM Length L Ch R = 1 ,36684   ,478,478,478
BEGIN DESCRIPTION:
WHEELOCK CREEK 61.0
END DESCRIPTION:
XS GIS Cut Line= 4
      3663040.25     10503943.38      3663231.22     10503630.88
      3663482.95     10503509.35      3664741.67     10503526.72
#Sta/Elev= 30
  4149.8  348.53  4348.4  336.44  4406.5   325.6  4443.2   323.1  4665.6  325.04
  4812.2  315.47  4962.2  299.82  4999.2  282.35    5002  281.85  5005.2  282.35
  5012.2  283.09  5022.2  290.33  5042.2  282.72  5062.2  287.11  5082.3  282.85
  5092.3  284.92  5102.3  295.95  5112.3  296.73  5132.3  286.65  5142.3  286.59
  5162.3  292.66  5292.3  296.05  5552.3  309.89  5604.5  315.81  5652.3  313.67
  5662.3   318.5  5692.3  319.95    5704  323.66  5792.3  338.43  6054.4  362.89
#Mann= 5 ,-1 , 0
  4149.8     .05       0  4999.2     .03       0  5005.2     .05       0
  5604.5     .08       0    5704     .16       0
Bank Sta=4962.2,5112.3
XS Rating Curve= 0 ,0
Exp/Cntr=0.3,0.1

Type RM Length L Ch R = 1 ,36206   ,491,491,491
BEGIN DESCRIPTION:
WHEELOCK CREEK 60.0
END DESCRIPTION:
XS GIS Cut Line= 3
      3663199.56     10503910.19      3663599.61     10503910.19
      3664349.61     10504060.19
#Sta/Elev= 30
  4550.2  336.66  4620.2  331.32  4670.2  330.34  4770.2  320.53  4810.2  315.52
  4850.2  302.38  4868.1  300.44  4880.2  299.76  4930.2  291.96  4960.4  289.61
  4998.2  280.56    5001  280.06  5004.2  280.56  5014.3  283.45  5031.8  296.05
    5042  297.99  5113.4  298.16  5184.8  292.86  5290.1  294.99  5378.6  299.66
  5434.6  305.52  5500.9  315.53  5534.6  315.03  5582.5  314.75  5602.9   316.8
  5623.3  322.53  5633.5  331.94  5653.4  335.89  5704.9   344.7  5715.1  344.53
#Mann= 9 ,-1 , 0
  4550.2     .05       0  4868.1     .16       0  4998.2     .07       0
  5004.2     .16       0  5014.3     .05       0  5290.1     .16       0
  5434.6     .05       0  5534.6     .16       0  5653.4     .08       0
Bank Sta=4880.2,5042
XS Rating Curve= 0 ,0
Exp/Cntr=0.3,0.1

Type RM Length L Ch R = 1 ,35715   ,210,210,210
BEGIN DESCRIPTION:
WHEELOCK CREEK 59.0
END DESCRIPTION:
XS GIS Cut Line= 4
      3663048.94      10504073.6       3663326.7     10504273.24
      3664229.48     10504360.05      3664680.87     10504490.26
#Sta/Elev= 30
  4333.9  346.05  4468.9  335.22  4700.1  304.15  4889.8  297.67  4910.1  290.85
  4940.1  296.89  4970.2  292.06  4997.4  279.24  5000.1  278.74  5003.4  279.24
  5030.5  289.01  5115.1  288.34    5141  293.57  5161.1  288.18  5181.2  294.18
  5452.4  308.38  5512.9  316.28  5612.7  329.66  5706.2  343.31  5817.6  350.32
  5832.8  354.88  5851.2  351.26  5856.4  355.51  5890.1  354.89  5895.3  358.85
  5928.9  362.01  5996.2   363.3  6001.4  368.55  6029.9  367.31  6052.7  372.89
#Mann= 6 ,-1 , 0
  4333.9     .05       0  4889.8     .16       0  4997.4     .07       0
  5003.4     .16       0  5512.9     .08       0  5612.7     .16       0
Bank Sta=4970.2,5030.5
XS Rating Curve= 0 ,0
Exp/Cntr=0.3,0.1

Type RM Length L Ch R = 1 ,35505   ,629,629,629
BEGIN DESCRIPTION:
Mapping XS 1b36ded2
END DESCRIPTION:
XS GIS Cut Line= 3
      3662404.23     10505122.64      3663775.81      10504462.9
      3664309.68     10504436.85
#Sta/Elev= 30
  3585.7  384.44  3939.1  372.62    4109  370.27  4290.1   346.8    4324   345.5
  4346.5  349.99  4357.3  342.94  4423.9  340.61  4509.4  327.59  4641.9  308.57
  4812.3  297.46  4940.4  296.38  4978.8   287.5  4985.7  281.28  4991.2  284.35
  4997.9  278.84  5000.7  278.34  5003.9  278.84  5013.9  278.99  5030.9   292.4
  5045.3  295.33  5121.5  294.87  5141.5  287.92  5151.6  292.49  5321.8  300.46
  5488.6  315.63    5532  318.25    5542  327.16  5587.8  332.68  5642.2   342.5
#Mann= 8 ,-1 , 0
  3585.7     .05       0  3939.1     .16       0  4509.4     .05       0
  4641.9     .16       0  4997.9     .07       0  5003.9     .16       0
  5488.6     .08       0  5587.8     .16       0
Bank Sta=4940.4,5045.3
XS Rating Curve= 0 ,0
Exp/Cntr=0.3,0.1

Type RM Length L Ch R = 1 ,34876   ,251,251,251
BEGIN DESCRIPTION:
WHEELOCK CREEK 58.0
END DESCRIPTION:
XS GIS Cut Line= 6
      3663059.68     10506285.79      3663788.83     10505556.65
      3663923.38     10505061.86      3664031.88      10504797.1
      3664092.65     10504562.72      3664439.83     10504445.55
#Sta/Elev= 30
  3381.2  373.63    3470  373.16  3512.4  366.21  3540.7  357.75  3696.2  347.27
  3809.4  343.14  3915.4  334.56  4049.8   331.9  4247.8  304.97    4553  296.12
  4735.3  291.76  4742.4  294.01  4937.7   292.1  4948.5  290.28  4954.3  283.65
  4957.7  285.73  5004.7  278.35  5007.5  277.85  5010.7  278.35  5045.8  293.04
  5114.1  295.28  5228.7  302.13  5249.4  298.61  5266.7  302.34    5363   309.3
  5418.9  309.33  5545.2  316.04  5622.3  332.61  5723.2  347.61  5819.8  353.68
#Mann= 10 ,-1 , 0
  3381.2     .16       0    4553     .05       0  4735.3     .16       0
  4957.7     .08       0  5004.7     .07       0  5010.7     .08       0
  5114.1     .16       0  5266.7     .08       0  5418.9     .05       0
  5622.3     .16       0
Bank Sta=4937.7,5045.8
XS Rating Curve= 0 ,0
Exp/Cntr=0.3,0.1

Type RM Length L Ch R = 1 ,34625   ,549,549,549
BEGIN DESCRIPTION:
WHEELOCK CREEK 57.0
END DESCRIPTION:
XS GIS Cut Line= 4
      3663636.93     10506502.79      3663927.72     10505587.03
      3664096.99       10505153.       3664504.8     10504558.64
#Sta/Elev= 30
  3634.2  373.92  3661.4  372.25  3693.6  353.07  3763.4  346.76  3797.9  350.05
  3799.3  349.97  3846.8   347.8  3887.2  350.44  3930.7  339.77  4001.3   339.6
    4103  333.39  4171.6  326.99  4329.4  307.39  4471.2  302.11    4581  298.79
  4833.7  291.67  4966.9  292.69    4978   280.3  4988.8  285.26  4999.1  276.04
  5001.8  275.54  5005.1  276.04  5010.2  276.99  5031.9  294.43  5051.1  299.62
    5180  302.17  5209.8  299.76  5294.7  306.29  5380.3  319.51  5781.7  363.55
#Mann= 10 ,-1 , 0
  3634.2     .16       0  3797.9     .05       0  3799.3     .16       0
  4001.3     .05       0    4103     .08       0  4171.6     .16       0
  4471.2     .05       0    4581     .16       0  4999.1     .07       0
  5005.1     .16       0
Bank Sta=4966.9,5031.9
XS Rating Curve= 0 ,0
Exp/Cntr=0.3,0.1

Type RM Length L Ch R = 1 ,34076   ,592,592,592
BEGIN DESCRIPTION:
WHEELOCK CREEK 56.0
END DESCRIPTION:
XS GIS Cut Line= 3
      3663728.06     10506567.94      3664299.61     10505660.19
       3664899.6      10505260.2
#Sta/Elev= 30
  3892.2  379.02  3948.6  372.54  3957.7  357.55  3978.9  352.75  4130.8  349.06
  4196.8  343.78  4428.6  319.61  4480.4  308.02  4586.8  295.77  4726.5  291.36
  4951.3  293.25  4957.3  293.37    4962  283.74  4972.4  283.49  4978.4  276.82
    4998  275.03  5000.7  274.53    5004  275.03  5008.5  275.13  5014.5  282.17
  5023.5  282.31  5050.5  293.08  5152.7  291.67  5325.5   307.8  5397.6  321.51
  5513.2  357.89  5564.3   364.6  5577.8  369.98  5585.4  384.14    5686  404.44
#Mann= 3 ,-1 , 0
  3892.2     .16       0    4998     .07       0    5004     .16       0
Bank Sta=4951.3,5050.5
XS Rating Curve= 0 ,0
Exp/Cntr=0.3,0.1

Type RM Length L Ch R = 1 ,33484   ,400,400,400
BEGIN DESCRIPTION:
WHEELOCK CREEK 55.0
END DESCRIPTION:
XS GIS Cut Line= 3
      3664240.24      10506654.7       3664583.1     10506099.18
       3664949.6      10505410.2
#Sta/Elev= 30
    4247   338.9  4475.6  328.52  4619.8  314.27  4635.2  310.39  4656.4  310.39
    4699  301.29  4781.1  292.84  4845.6  289.04  4888.2  291.42  4899.8  290.14
  4903.7  284.01    4920  285.74  4925.6   282.7  4985.9  283.83  4991.6  278.27
  5004.9  274.09  5007.6  273.59  5010.9  274.09  5023.3  279.33  5035.5  291.37
  5243.9  291.27  5353.8  302.21  5408.4  312.73    5436  325.59  5487.7  331.66
  5540.2  358.14  5589.8  375.69  5622.4  381.26  5634.9   386.6  5680.2  393.03
#Mann= 3 ,-1 , 0
    4247     .16       0  5004.9     .07       0  5010.9     .16       0
Bank Sta=4985.9,5035.5
XS Rating Curve= 0 ,0
Exp/Cntr=0.3,0.1

Type RM Length L Ch R = 1 ,33084   ,663,663,663
BEGIN DESCRIPTION:
WHEELOCK CREEK 54.0
END DESCRIPTION:
XS GIS Cut Line= 3
      3664340.01     10506802.34      3664904.28     10506216.37
      3665049.62     10505510.16
#Sta/Elev= 30
  4234.5   339.8  4384.3  329.61  4433.7   329.5  4628.6   318.4  4815.7  297.31
  4850.9  290.88  4886.5  288.01    4950  290.47  4957.2  288.93  4964.1  284.89
  4978.3  282.61  5003.6  273.66  5006.3  273.16  5009.6  273.66  5013.8  274.45
  5020.7  281.11  5041.9  284.23  5054.5  289.95  5104.1  290.47  5340.2  295.25
  5401.7  299.74  5563.6  319.63    5626  332.27  5643.1  339.25  5648.2  339.19
  5666.9  349.67  5698.6     360  5707.7  365.36  5743.8  374.66    5769  378.63
#Mann= 6 ,-1 , 0
  4234.5      .1       0  4628.6     .16       0  5003.6     .07       0
  5009.6     .16       0  5104.1      .1       0  5563.6     .16       0
Bank Sta=4957.2,5054.5
XS Rating Curve= 0 ,0
Exp/Cntr=0.3,0.1

Type RM Length L Ch R = 1 ,32421   ,583,583,583
BEGIN DESCRIPTION:
WHEELOCK CREEK 53.0
END DESCRIPTION:
XS GIS Cut Line= 3
      3664649.59     10506910.19      3665049.61     10506760.19
      3665849.61     10506010.19
#Sta/Elev= 30
  4584.1   322.6  4709.6  308.96  4739.9   308.3  4770.1  312.22    4787  310.71
  4808.4  313.06  4840.4  311.43  4885.8  304.16  4910.7  296.04  4957.9  290.23
  4971.3  287.11  4979.3  280.11    4990  276.45  4993.2  272.48  4995.9  271.98
  4999.2  272.48  5008.6  274.74  5018.4  272.65  5025.3  275.85  5032.6  275.79
  5039.4  280.81  5081.9  288.23  5188.4   290.2  5308.5  288.46  5346.3  290.53
  5389.4  291.82  5725.7  297.63  5888.6  311.05    6030  331.66  6107.9  335.87
#Mann= 5 ,-1 , 0
  4584.1     .16       0  4993.2     .07       0  4999.2     .16       0
  5346.3     .12       0  5389.4     .16       0
Bank Sta=4957.9,5081.9
XS Rating Curve= 0 ,0
Exp/Cntr=0.3,0.1

Type RM Length L Ch R = 1 ,31838   ,596,596,596
BEGIN DESCRIPTION:
WHEELOCK CREEK 52.0
END DESCRIPTION:
XS GIS Cut Line= 3
      3665249.61      10507710.2      3665449.61     10506960.19
      3666002.34     10506138.28
#Sta/Elev= 30
  4232.6  334.89  4263.7  329.08  4284.4  330.28  4485.5  309.19  4525.6  301.08
  4605.8  290.72  4646.6  287.36  4683.5   288.8  4812.2  289.96  4851.4  288.05
  4898.6  290.05    4926  289.48  4957.1  281.09  4977.8  279.82  4995.5  272.03
  4998.2  271.53  5001.5  272.03  5011.8  273.02  5016.3  278.47  5037.3  286.61
    5045   287.1  5073.3  289.59    5155  287.92  5310.3  289.79  5454.7  301.45
  5556.3   313.3  5658.2  315.95  5715.2  319.21  5772.2  325.76  5999.3  336.94
#Mann= 7 ,-1 , 0
  4232.6     .16       0  4683.5     .12       0  4851.4     .16       0
  4898.6     .12       0  4995.5     .07       0  5001.5     .12       0
    5155     .16       0
Bank Sta=4926,5045
XS Rating Curve= 0 ,0
Exp/Cntr=0.3,0.1

Type RM Length L Ch R = 1 ,31242   ,655,655,655
BEGIN DESCRIPTION:
WHEELOCK CREEK 51.0
END DESCRIPTION:
XS GIS Cut Line= 3
       3665507.6     10507974.14      3665781.02     10507431.65
      3666024.07     10506368.27
#Sta/Elev= 30
  4340.8  336.62    4614  322.82  4703.6  311.98  4738.4  309.88  4777.4  302.26
  4844.4  293.25  4911.3  286.82  4959.7  285.29  4980.6  276.07  4998.1  271.07
  5000.8  270.57  5004.1  271.07  5012.9  272.27  5021.6  277.04  5031.9  279.97
  5042.1  281.07  5055.8  288.26  5134.4  286.67  5184.7   288.6  5239.1  287.71
  5247.3  288.36  5275.7  285.74  5298.6   287.3  5465.2  287.98  5616.6  299.84
  5677.7  301.64  5688.4  300.71  5730.9  303.38    5956   324.6  6039.1  329.24
#Mann= 5 ,-1 , 0
  4340.8     .16       0  4998.1     .07       0  5004.1     .16       0
  5239.1     .12       0  5465.2     .16       0
Bank Sta=4959.7,5055.8
XS Rating Curve= 0 ,0
Exp/Cntr=0.3,0.1

Type RM Length L Ch R = 1 ,30587   ,342,342,342
BEGIN DESCRIPTION:
WHEELOCK CREEK 50.0
END DESCRIPTION:
XS GIS Cut Line= 3
      3666171.42     10508201.11      3666206.14     10507770.52
      3667045.55      10506910.3
#Sta/Elev= 30
  4336.1  319.79  4457.4  319.46  4496.4  316.69  4501.4  317.54  4517.6  314.06
    4638  299.34  4738.3  292.22  4765.8  288.38  4862.7  284.68  4940.5  286.76
  4954.6  285.43  4961.8  281.64  4982.9  275.33    4994  270.37  4996.8  269.87
    5000  270.37  5011.2  270.45  5018.3  275.12  5053.6  286.83  5066.4  287.43
  5083.4  287.45  5202.1  285.16  5329.4  285.87    5485  301.46  5506.3  305.46
  5646.5   321.2  5760.7  334.17  5905.1  345.04  5941.4  347.52    5970  351.48
#Mann= 8 ,-1 , 0
  4336.1     .16       0    4994     .07       0    5000     .16       0
  5066.4     .12       0  5083.4     .16       0  5646.5     .05       0
  5905.1      .1       0  5941.4     .05       0
Bank Sta=4954.6,5053.6
XS Rating Curve= 0 ,0
Exp/Cntr=0.3,0.1

Type RM Length L Ch R = 1 ,30245   ,505,505,505
BEGIN DESCRIPTION:
WHEELOCK CREEK 49.0
END DESCRIPTION:
XS GIS Cut Line= 3
       3666499.6     10508110.21      3666649.61     10507710.19
      3667099.63     10507160.16
#Sta/Elev= 30
  4594.9  308.18  4665.2  297.77  4819.2  283.95  4841.5  283.18    4861   286.1
    4958  284.79  4968.7  280.86  4976.7  274.89  4982.1  278.77  4990.1  270.56
  5009.3  270.05  5012.1  269.55  5015.3  270.05  5025.4  270.36  5029.3  275.11
  5035.8  270.75    5058   277.6  5064.5  275.82  5072.4  279.87  5078.8  278.55
  5136.3  284.76    5221   284.9  5448.5  297.87  5455.7  300.62  5533.9  308.64
  5590.6  321.25  5597.8  320.25  5604.3  323.93  5696.5  337.88  5732.8  342.34
#Mann= 4 ,-1 , 0
  4594.9     .16       0  5009.3     .07       0  5015.3     .16       0
  5696.5     .05       0
Bank Sta=4982.1,5029.3
XS Rating Curve= 0 ,0
Exp/Cntr=0.3,0.1

Type RM Length L Ch R = 1 ,29740   ,584,584,584
BEGIN DESCRIPTION:
WHEELOCK CREEK 48.0
END DESCRIPTION:
XS GIS Cut Line= 2
      3666615.87      10508409.4      3667393.66      10507319.1
#Sta/Elev= 30
  4570.8  318.96  4631.3     319    4694  315.98  4794.8  306.21  4895.6  292.65
  4901.7  289.96    4946  286.76  4952.1  288.66  4966.9  286.07  4981.6  270.42
  4993.4  268.37  4996.1  267.87  4999.4  268.37  5017.3   272.5    5032  280.53
  5052.9  284.98  5218.8  285.48  5355.3  282.42    5477  286.46  5640.4  304.35
  5684.7  318.66  5705.6  320.09  5720.3  325.44  5752.4   330.2    5756  331.52
  5762.1  329.57  5770.7  332.65  5791.6  334.32  5856.8  345.92  5910.1  349.45
#Mann= 4 ,-1 , 0
  4570.8     .16       0  4993.4     .07       0  4999.4     .16       0
  5752.4     .05       0
Bank Sta=4966.9,5052.9
XS Rating Curve= 0 ,0
Exp/Cntr=0.3,0.1

Type RM Length L Ch R = 1 ,29156   ,641,641,641
BEGIN DESCRIPTION:
WHEELOCK CREEK 47.0
END DESCRIPTION:
XS GIS Cut Line= 3
       3666899.6     10508510.19      3667249.61     10508310.19
      3667749.63     10507610.15
#Sta/Elev= 30
  4613.1  317.95  4664.2  314.42  4751.3  299.34  4884.5  284.71  4943.5  280.82
  4949.3  283.32  4965.1  279.23  4970.9  283.42  4986.7  276.89  4993.2  268.56
  4999.5  267.63  5002.3  267.13  5005.5  267.63  5008.3   267.7  5013.3  272.74
  5019.3  272.74  5023.6  275.82  5065.4  281.55  5075.2  283.78  5201.8   281.3
  5468.5  283.49  5596.3  289.63  5672.7  299.71  5682.3  300.98  5726.5  315.17
  5732.7  320.77  5768.3  334.26  5812.6   354.9  5839.6  360.29  5876.5     362
#Mann= 5 ,-1 , 0
  4613.1     .16       0  4999.5     .07       0  5005.5     .16       0
  5075.2     .05       0  5672.7     .16       0
Bank Sta=4970.9,5065.4
XS Rating Curve= 0 ,0
Exp/Cntr=0.3,0.1

Type RM Length L Ch R = 1 ,28515   ,428,428,428
BEGIN DESCRIPTION:
WHEELOCK CREEK 46.0
END DESCRIPTION:
XS GIS Cut Line= 3
      3667025.58     10509423.31      3667629.76     10508659.41
      3668303.36     10508089.97
#Sta/Elev= 30
  4324.5  316.27  4386.6  314.87  4465.2  309.48    4558  293.94  4685.5  282.05
  4934.8  282.12  4963.7  280.09    4970  279.53  4978.1  269.02  4988.5  266.93
  4991.2  266.43  4994.5  266.93  5005.3  268.55  5042.2  280.33  5489.5   281.7
  5659.8  293.86  5735.5  302.74  5836.7  304.75    5873  310.33  5879.5  314.38
  5908.1  322.69  5914.7  321.67  5971.8   327.7  5976.9  329.88  6035.5  342.22
  6070.8  353.36    6107   357.5  6113.6  359.96  6180.1  363.95  6180.5  363.95
#Mann= 6 ,-1 , 0
  4324.5     .05       0  4988.5     .07       0  4994.5     .05       0
  5735.5     .05       0  5976.9     .16       0  6180.1     .05       0
Bank Sta=4963.7,5042.2
XS Rating Curve= 0 ,0
Exp/Cntr=0.3,0.1

Type RM Length L Ch R = 1 ,28087   ,783,783,783
BEGIN DESCRIPTION:
WHEELOCK CREEK 45.0
END DESCRIPTION:
XS GIS Cut Line= 3
      3667091.81     10509640.82      3667660.36     10509219.84
      3668353.97     10508504.55
#Sta/Elev= 30
  4034.9  314.21  4141.6   312.6  4212.5  314.26  4333.5  301.09  4412.9  288.32
    4505  279.35  4882.9  281.02  4939.5  278.87    4982  272.59  4989.1  266.99
  4993.1  266.87  4995.8  266.37  4999.1  266.87    5002  266.97  5010.2  272.76
  5024.4  277.45    5081  273.76  5088.2  274.28  5095.1  279.17  5222.5  288.81
  5264.9  295.93  5271.9  299.25  5342.6  314.66  5390.6  317.75  5540.7   330.2
    5562  333.84  5611.4  336.55  5653.8   343.2  5682.1  353.06  5738.7   360.3
#Mann= 5 ,-1 , 0
  4034.9     .05       0  4993.1     .03       0  4999.1     .05       0
    5002     .16       0  5390.6     .05       0
Bank Sta=4939.5,5024.4
XS Rating Curve= 0 ,0
Exp/Cntr=0.3,0.1

Type RM Length L Ch R = 1 ,27304   ,402,402,402
BEGIN DESCRIPTION:
WHEELOCK CREEK 44.0
END DESCRIPTION:
XS GIS Cut Line= 4
      3667084.63     10510043.08      3667579.41     10509817.39
      3668629.76      10509635.1      3669011.66     10509912.85
#Sta/Elev= 30
  4069.9  317.59  4251.2  315.13  4339.2  316.27  4460.1  312.72    4504  304.51
  4747.3  283.66  4898.1  277.18  4916.2  274.66  4928.6  277.18  4975.9  277.12
  4980.9  271.85  4996.6  265.67  4999.4  265.17  5002.6  265.67  5006.7  266.07
  5040.6  276.35  5101.1  278.95  5209.5  278.71    5233  278.32  5253.3  274.31
  5269.2  276.66  5274.3  274.89  5293.9  277.44  5326.5  277.75  5537.5  279.13
  5696.7  292.53  5854.4   312.7  5926.9  330.74  5963.4  337.45    6152  349.65
#Mann= 6 ,-1 , 0
  4069.9     .05       0  4996.6     .03       0  5002.6     .05       0
  5006.7     .16       0  5326.5     .05       0  5696.7     .16       0
Bank Sta=4975.9,5040.6
XS Rating Curve= 0 ,0
Exp/Cntr=0.3,0.1

Type RM Length L Ch R = 1 ,26902   ,307,307,307
BEGIN DESCRIPTION:
WHEELOCK CREEK 43.0
END DESCRIPTION:
XS GIS Cut Line= 4
      3667261.03     10510322.28      3667803.59     10510148.66
      3668211.57     10510122.62      3668871.27     10509940.33
#Sta/Elev= 30
  4169.2  319.98  4262.8   314.4  4346.2  312.17  4398.7  313.41  4482.6   310.5
  4589.6  301.86  4616.5  295.83  4621.7  298.05  4648.6  292.17    4686  291.73
  4791.7  280.99  4875.2   276.4  4925.3  277.43  4955.3  275.52  4975.4  272.61
  4995.4  264.72  5002.4  264.33  5005.2  263.83  5008.4  264.33  5025.5  274.14
  5055.5  277.41  5218.3   275.6  5326.5  278.38  5536.4  298.71  5612.5   307.4
  5640.1  313.34  5693.6  323.63  5706.1  327.39  5747.4  333.45  5832.1  340.56
#Mann= 6 ,-1 , 0
  4169.2     .05       0  5002.4     .03       0  5008.4     .05       0
  5536.4     .16       0  5640.1     .05       0  5693.6     .16       0
Bank Sta=4955.3,5025.5
XS Rating Curve= 0 ,0
Exp/Cntr=0.3,0.1

Type RM Length L Ch R = 1 ,26595   ,714,714,714
BEGIN DESCRIPTION:
WHEELOCK CREEK 42.0
END DESCRIPTION:
XS GIS Cut Line= 5
      3667226.35     10510782.33      3667742.82      10510487.2
      3667912.09     10510439.46      3668228.93     10510387.38
      3668832.22     10510218.11
#Sta/Elev= 30
  4109.1  324.69  4529.9  311.21    4648  292.59  4703.9  287.86  4721.4  282.07
  4744.7  278.91    4928  274.47  4953.1  271.41  4970.7  271.76  4995.9  263.95
  4998.7  263.45  5001.9  263.95    5009  263.96  5026.8  274.41  5031.9  271.68
  5039.5  276.24  5049.6  276.56  5232.8  277.15  5433.2  283.16    5669  317.42
  5687.4   317.2  5692.6  321.32  5700.2  322.74  5726.7  316.27  5741.7  321.15
  5760.8  318.62  5800.1  330.67  5805.2  326.69  5814.4     332  5827.5  332.62
#Mann= 5 ,-1 , 0
  4109.1     .16       0  4744.7     .05       0  4953.1     .16       0
  4995.9     .07       0  5001.9     .16       0
Bank Sta=4928,5026.8
XS Rating Curve= 0 ,0
Exp/Cntr=0.3,0.1

Type RM Length L Ch R = 1 ,25881   ,531,531,531
BEGIN DESCRIPTION:
WHEELOCK CREEK 41.0
END DESCRIPTION:
XS GIS Cut Line= 3
      3667649.62     10510960.19      3668299.61     10510810.19
      3668799.62     10510610.18
#Sta/Elev= 30
  4346.6   309.5  4365.4  307.44  4377.4  302.77  4387.6  301.64  4397.9  296.79
  4418.4  290.93  4461.2  284.06    4510  278.64  4562.1   275.9    4845  274.57
    4870  273.24  4931.6  275.02  4972.6  273.61  4982.9  272.17  4994.9  262.75
  5000.4  262.09  5003.2  261.59  5006.4  262.09  5011.1  264.96  5016.4  264.96
  5035.2  274.42  5052.7  273.46  5229.1  283.31  5261.4  288.78  5273.5  289.11
  5304.5   294.3  5390.6  304.25  5476.8   317.1  5483.5  319.65  5552.2  327.57
#Mann= 5 ,-1 , 0
  4346.6     .16       0    4510     .05       0    4845     .16       0
  5000.4     .07       0  5006.4     .16       0
Bank Sta=4972.6,5035.2
XS Rating Curve= 0 ,0
Exp/Cntr=0.3,0.1

Type RM Length L Ch R = 1 ,25350   ,559,559,559
BEGIN DESCRIPTION:
WHEELOCK CREEK 40.0
END DESCRIPTION:
XS GIS Cut Line= 3
      3667799.63     10511360.19      3668549.61     10511260.19
      3669680.36     10510491.52
#Sta/Elev= 30
  4226.6  309.74  4261.6  307.81  4357.7  286.09  4579.7  271.45  4670.7  270.97
  4871.2  273.17  4946.7  273.36  4986.2   270.4  4996.7  261.25  5002.6  261.06
  5005.4  260.56  5008.6  261.06  5019.5  270.83  5032.7  273.26    5314  272.11
  5387.2  279.76  5574.4  294.84  5709.2  316.28  5825.9  313.71  5969.6  323.43
  6077.3  347.34  6092.3  343.75  6113.3  347.43  6143.1  340.05  6179.1  348.17
  6185.1  354.63  6200.1  354.65  6206.1  359.81    6236  359.43  6350.5  378.82
#Mann= 7 ,-1 , 0
  4226.6     .05       0  4261.6     .16       0  4670.7     .12       0
  4871.2     .05       0  5002.6     .03       0  5008.6     .05       0
  5387.2     .16       0
Bank Sta=4946.7,5032.7
XS Rating Curve= 0 ,0
Exp/Cntr=0.3,0.1

Type RM Length L Ch R = 1 ,24791   ,516,516,516
BEGIN DESCRIPTION:
WHEELOCK CREEK 39.0
END DESCRIPTION:
XS GIS Cut Line= 3
      3667299.62     10513210.18      3668899.61     10511660.19
      3669699.63     10510960.17
#Sta/Elev= 30
  2799.7  370.22  3153.3  341.16  3499.8  318.52  3697.8  308.48  3846.3  280.67
  3952.5  269.62  4256.5  271.45  4277.7  266.94    4299   270.8  4581.8   268.7
  4963.7  272.57    4985  268.81    4992  265.42  4996.2  260.21  4998.9  259.71
  5002.2  260.21  5013.3  260.34  5020.3  269.15  5027.4  271.49  5431.2  269.38
  5610.7  273.86  5729.2  283.04  5849.8  302.39  5870.7  311.71  5891.5  317.09
  5913.4  318.37  5991.2  353.34  5997.8  358.46  6038.6  366.16  6090.4  369.97
#Mann= 5 ,-1 , 0
  2799.7     .05       0  4996.2     .03       0  5002.2     .05       0
  5610.7     .16       0  6038.6      .1       0
Bank Sta=4963.7,5027.4
XS Rating Curve= 0 ,0
Exp/Cntr=0.3,0.1

Type RM Length L Ch R = 1 ,24275   ,511,511,511
BEGIN DESCRIPTION:
WHEELOCK CREEK 38.0
END DESCRIPTION:
XS GIS Cut Line= 3
      3667966.77     10512882.17      3668999.61     10512160.19
      3669982.44     10511965.49
#Sta/Elev= 30
  3722.9  323.19  3927.4  311.06    4007  302.91  4054.5  293.25  4098.3  287.96
    4264  270.62  4609.4  269.75  4624.2  269.36  4630.3  264.56  4671.1   266.4
  4701.6  269.09  4975.7  270.63  5005.7  259.52  5008.4  259.02  5011.7  259.52
  5044.2  269.78  5095.2  271.18    5136  279.71  5162.3  274.34  5167.4  277.33
  5207.3  275.24  5218.6  277.69  5237.9  272.93  5259.8  272.61  5339.9  273.74
  5628.4  295.44  5808.8  317.53  5910.7   347.4  5935.7  348.02    5985  342.14
#Mann= 8 ,-1 , 0
  3722.9     .05       0  4054.5     .16       0  4098.3     .05       0
  4671.1     .12       0  4701.6     .05       0  5005.7     .03       0
  5011.7     .05       0  5259.8     .16       0
Bank Sta=4975.7,5044.2
XS Rating Curve= 0 ,0
Exp/Cntr=0.3,0.1

Type RM Length L Ch R = 1 ,23764   ,569,569,569
BEGIN DESCRIPTION:
WHEELOCK CREEK 37.0
END DESCRIPTION:
XS GIS Cut Line= 3
      3667883.24      10513406.8      3669199.61     10512610.19
      3669599.65     10512410.17
#Sta/Elev= 30
  3450.6  346.72  3670.2  331.66  3960.9  316.39  4065.9  311.81    4136  304.53
  4166.8  297.63  4194.4  295.39  4252.8  282.42  4356.9  271.34  4428.2  267.96
  4881.8  269.49  4954.2  270.29  4981.5  265.19  4986.3   258.7  4994.6   258.6
  4997.4   258.1  5000.6   258.6  5003.2  258.66  5011.6     267    5034  270.64
  5078.7  268.43  5087.1  271.22  5145.8  273.25  5271.5  287.32  5316.3  300.93
  5369.4  324.44  5383.3  327.72  5405.7  337.36  5414.1  343.05  5436.5  346.75
#Mann= 6 ,-1 , 0
  3450.6     .05       0  3960.9     .16       0  4252.8     .05       0
  4881.8     .16       0  4994.6     .07       0  5000.6     .16       0
Bank Sta=4954.2,5034
XS Rating Curve= 0 ,0
Exp/Cntr=0.3,0.1

Type RM Length L Ch R = 1 ,23195   ,596,596,596
BEGIN DESCRIPTION:
WHEELOCK CREEK 36.0
END DESCRIPTION:
XS GIS Cut Line= 3
      3668299.59     10513910.21      3669099.61     10513160.19
      3669599.57     10512810.21
#Sta/Elev= 30
  3882.2   349.1    4031  333.52    4158  323.96  4375.9  299.98  4384.6  296.55
  4455.4  287.44  4540.2  282.67  4547.3  278.84  4554.1  281.54  4568.3  281.22
  4683.5  272.95  4830.1  266.36  4971.7   268.1  4981.9  266.64  4986.2  261.79
  4992.3  261.41    4998  257.97  5000.8  257.47    5004  257.97  5015.4  261.05
    5022  266.59  5028.1   267.8  5173.7   268.2  5222.9  271.14  5234.9  275.46
  5259.6  276.82  5316.7  288.14  5421.1  302.03  5510.2  313.94  5589.1  321.53
#Mann= 7 ,-1 , 0
  3882.2     .05       0  4375.9     .16       0  4683.5     .05       0
    4998     .03       0    5004     .05       0  5234.9     .12       0
  5421.1     .16       0
Bank Sta=4971.7,5028.1
XS Rating Curve= 0 ,0
Exp/Cntr=0.3,0.1

Type RM Length L Ch R = 1 ,22599   ,548,548,548
BEGIN DESCRIPTION:
WHEELOCK CREEK 35.0
END DESCRIPTION:
XS GIS Cut Line= 3
      3669358.92     10514209.77      3669449.61     10513560.19
      3669649.61     10512860.18
#Sta/Elev= 30
  4353.1  308.54  4462.6  308.48  4539.2  305.82    4595  297.24  4610.7  286.71
  4615.7  286.89  4625.3  283.32  4635.4  286.35  4645.5  285.77  4753.7  273.89
  4867.6  266.43  4973.2  266.97  4988.8  257.84  5003.5  257.05  5006.2  256.55
  5009.5  257.05  5019.4     261  5025.9  267.02  5031.1   267.9  5123.4  268.29
  5144.2  265.83  5234.6  268.21  5310.6  265.98  5362.6  266.95  5463.5  279.72
  5574.5  293.88    5581  296.44    5633  304.83  5642.1  307.88    5737  320.22
#Mann= 5 ,-1 , 0
  4353.1     .05       0  5003.5     .03       0  5009.5     .05       0
  5234.6     .05       0  5463.5     .16       0
Bank Sta=4973.2,5031.1
XS Rating Curve= 0 ,0
Exp/Cntr=0.3,0.1

Type RM Length L Ch R = 1 ,22051   ,476,476,476
BEGIN DESCRIPTION:
WHEELOCK CREEK 34.0
END DESCRIPTION:
XS GIS Cut Line= 3
      3670149.64     10514060.22      3669849.61     10513760.19
      3669699.62     10512960.24
#Sta/Elev= 30
  4575.5  305.12    4618  305.81  4674.5  302.15  4688.7  299.16  4731.1  294.04
  4801.8  286.65    4816  283.96  4844.2  281.96  4957.4  266.07  4971.5  265.59
  4985.7  258.46  4993.3  257.45    4996  256.95  4999.3  257.45    5010  259.35
  5022.8  264.34  5026.1  266.29  5110.4  266.71    5112  266.69  5498.3  266.37
  5589.9  270.09  5624.7  272.87  5661.1  280.66  5696.9  285.33  5752.7  294.54
  5773.1  298.68  5782.4  302.26  5787.5  302.14  5803.6  306.55  5813.7  307.57
#Mann= 7 ,-1 , 0
  4575.5     .16       0  4993.3     .07       0  4999.3     .16       0
  5022.8     .05       0  5110.4     .12       0    5112     .05       0
  5696.9     .16       0
Bank Sta=4971.5,5026.1
XS Rating Curve= 0 ,0
Exp/Cntr=0.3,0.1

Type RM Length L Ch R = 1 ,21575   ,381,381,381
BEGIN DESCRIPTION:
WHEELOCK CREEK 33.0
END DESCRIPTION:
XS GIS Cut Line= 3
      3670199.62     10513960.15      3670300.11     10513679.04
      3669799.59     10512760.15
#Sta/Elev= 30
  4668.4  300.51  4732.1  295.14  4770.8  288.69  4863.1  279.28  4870.1  276.78
  4969.1  266.24  4974.9  264.43  4980.6  263.52  4988.4  256.47  4993.7  255.81
  4996.5  255.31  4999.7  255.81  5018.6  261.27  5024.2   260.4  5040.4   265.2
  5122.8  266.11  5225.6  264.27  5476.3  266.17  5614.7  264.75  5660.2  269.16
  5710.8  276.51  5717.2  279.13    5740  281.29  5785.5  288.85  5814.3  298.52
    5829  299.51  5910.8  315.03  5933.5  316.78  5939.7  318.98  6013.3  322.46
#Mann= 5 ,-1 , 0
  4668.4     .16       0  4993.7     .07       0  4999.7     .16       0
  5122.8     .05       0    5829     .16       0
Bank Sta=4974.9,5040.4
XS Rating Curve= 0 ,0
Exp/Cntr=0.3,0.1

Type RM Length L Ch R = 1 ,21194   ,267,267,267
BEGIN DESCRIPTION:
Mapping XS a77bd0d8
END DESCRIPTION:
XS GIS Cut Line= 4
      3670206.35     10513986.35      3670513.65     10513585.29
      3670555.32     10513064.46      3671148.23     10511873.44
#Sta/Elev= 30
  4363.8  302.52  4618.4  275.55  4734.9  265.24  4974.5  265.01    5000  255.06
  5002.8  254.56    5006  255.06  5009.5  256.39  5025.4  260.99  5034.7  265.05
  5804.8     262  5908.8   262.7    5991  263.97  6094.4  269.03  6274.6  280.35
  6323.5  285.29  6330.7   288.8  6336.3  287.52  6358.7  293.91  6390.5  298.58
  6397.9  297.26  6403.5  300.22  6420.3  297.23  6502.2  303.32  6554.6  313.87
    6605  330.57  6649.8  336.31    6689  335.76  6694.6  338.92    6722  341.65
#Mann= 11 ,-1 , 0
  4363.8     .16       0  4618.4     .05       0    5000     .03       0
    5006     .05       0  5009.5     .16       0  5025.4     .05       0
  5804.8     .16       0  5908.8     .05       0    5991     .16       0
  6094.4     .05       0  6274.6     .16       0
Bank Sta=4974.5,5034.7
XS Rating Curve= 0 ,0
Exp/Cntr=0.3,0.1

Type RM Length L Ch R = 1 ,20927   ,719,719,719
BEGIN DESCRIPTION:
WHEELOCK CREEK 32.0
END DESCRIPTION:
XS GIS Cut Line= 3
      3670249.62     10514010.17      3670749.61     10513510.19
       3671549.6     10513110.19
#Sta/Elev= 30
  4289.6  300.19  4453.9  283.33  4699.7  264.29  4959.8  264.22  4968.4  263.71
  4982.5  256.47  4993.1  254.78  5005.1  254.69  5010.7  260.15  5027.4  262.78
  5053.4  263.91  5063.8  263.87  5072.2  257.76  5077.7  262.11  5086.1  260.27
  5091.5  254.24  5094.3  253.74  5097.5  254.24  5100.1  263.26  5116.9  256.55
  5130.8  261.22  5139.2  258.02  5144.8  262.59    5184   264.8  5541.7   259.8
  5636.8  264.05  5698.5  270.75  5748.6  275.76    5838  295.13  5891.1   317.3
#Mann= 7 ,-1 , 0
  4289.6     .16       0  4453.9     .05       0  4959.8     .16       0
  5053.4     .05       0  5091.5     .07       0  5097.5     .05       0
  5698.5     .16       0
Bank Sta=4968.4,5027.4
XS Rating Curve= 0 ,0
Exp/Cntr=0.3,0.1

Type RM Length L Ch R = 1 ,20208   ,395,395,395
BEGIN DESCRIPTION:
WHEELOCK CREEK 31.0
END DESCRIPTION:
XS GIS Cut Line= 3
       3670399.6     10514060.19      3671199.61     10513760.19
      3671549.62     10513460.18
#Sta/Elev= 30
  4124.9  284.02    4165  278.16  4295.8  265.52  4402.6  261.18  4453.9  261.18
  4620.1   260.9  4668.2   260.9  4775.4  261.83  4882.5  262.89  4969.5  262.54
  4976.6  253.92  5004.3  253.12    5007  252.62  5010.3  253.12    5015  255.63
  5021.6  253.49  5029.2  258.73  5035.8  256.11  5043.5  263.77  5135.7  262.43
  5142.3  259.67  5234.5  268.59  5269.6  278.54  5277.3  282.71  5312.4   289.1
  5334.4  296.27  5355.2  306.88  5369.5  317.59    5398  329.92  5440.3  336.27
#Mann= 8 ,-1 , 0
  4124.9     .05       0  4453.9     .12       0  4620.1     .16       0
  4668.2     .05       0  4775.4      .1       0  4882.5     .16       0
  5004.3     .07       0  5010.3     .16       0
Bank Sta=4969.5,5043.5
XS Rating Curve= 0 ,0
Exp/Cntr=0.3,0.1

Type RM Length L Ch R = 1 ,19813   ,478,478,478
BEGIN DESCRIPTION:
Mapping XS 7257c7bd
END DESCRIPTION:
XS GIS Cut Line= 4
      3670133.42     10514205.08      3670951.15     10514246.75
       3671602.2     10513788.42      3671898.31     10513123.46
#Sta/Elev= 30
  3481.9  297.45  3588.2  301.34  3628.3  298.17  3703.3  286.19  3918.7  267.32
  4045.6  264.42  4208.4  261.69  4533.3  259.15  4816.1  261.18  4971.4  262.36
  4985.3  253.24    4991   252.8  4993.8   252.3    4997   252.8    5021  262.68
    5057  262.09  5193.5  279.11    5200  283.29  5223.3  288.96  5275.2  298.34
    5292  304.69  5298.5  310.35  5313.9  314.89  5335.8  327.02  5357.7  330.95
  5373.7  330.75  5396.9  334.72  5478.1  334.63  5738.6  343.31  5824.8  343.13
#Mann= 7 ,-1 , 0
  3481.9     .16       0  3703.3     .05       0  4045.6     .16       0
  4208.4     .12       0  4816.1     .16       0    4991     .07       0
    4997     .16       0
Bank Sta=4971.4,5021
XS Rating Curve= 0 ,0
Exp/Cntr=0.3,0.1

Type RM Length L Ch R = 1 ,19335   ,372,372,372
BEGIN DESCRIPTION:
WHEELOCK CREEK 30.0
END DESCRIPTION:
XS GIS Cut Line= 4
      3670102.24     10514923.81      3671716.78     10514163.42
       3671914.7     10514054.04      3672154.29     10513147.75
#Sta/Elev= 30
  3122.7  301.47  3264.7  302.44  3395.9   292.4  3424.2  289.29    3447  283.26
    3521   281.4  3694.6  271.37  4011.7   263.7  4142.2  260.95  4494.9  258.62
  4627.2  258.13  4969.6  261.44    4996  251.42  4998.7  251.37  5001.4  250.87
  5004.7  251.37  5013.4  259.35  5023.4  261.39  5066.8  260.53    5173  259.02
  5274.7  265.58    5369  276.81  5509.8  298.37  5559.9  299.85  5605.4  294.58
  5645.6  294.39  5747.7  310.08    5756  313.91  5796.3  316.81  6070.9  322.62
#Mann= 11 ,-1 , 0
  3122.7     .16       0    3521     .05       0  4011.7     .16       0
  4142.2     .05       0  4494.9     .12       0  4627.2     .05       0
    4996     .16       0  4998.7     .07       0  5004.7     .16       0
  5066.8     .05       0  5274.7     .16       0
Bank Sta=4969.6,5023.4
XS Rating Curve= 0 ,0
Exp/Cntr=0.3,0.1

Type RM Length L Ch R = 1 ,18963   ,617,617,617
BEGIN DESCRIPTION:
WHEELOCK CREEK 29.0
END DESCRIPTION:
XS GIS Cut Line= 3
      3670449.58      10515010.2      3672049.61     10514360.19
      3672849.57     10513960.21
#Sta/Elev= 30
  3251.7  295.02  3327.3  289.44  3480.7  283.77  3552.9  284.06  3587.8  281.73
  3651.1  282.96  3689.5  280.92    3719   276.7  3844.8   272.8  4050.5  258.73
  4687.3  257.78  4943.8  260.05    4964  260.71  4969.4  257.52  4981.5  257.97
  4992.7  251.41  4998.1  251.01  5000.8  250.51  5004.1  251.01  5006.8  251.91
  5015.1  252.75  5031.8  260.58  5037.4  260.45  5135.2     258  5210.7  259.63
  5417.5  258.54  5503.3  265.01  5643.4  281.77  5678.9  286.17  5873.1  308.43
#Mann= 8 ,-1 , 0
  3251.7     .05       0  4943.8     .16       0  4998.1     .07       0
  5004.1     .16       0  5006.8     .05       0  5503.3      .1       0
  5643.4     .16       0  5678.9      .1       0
Bank Sta=4964,5037.4
XS Rating Curve= 0 ,0
Exp/Cntr=0.3,0.1

Type RM Length L Ch R = 1 ,18346   ,689,689,689
BEGIN DESCRIPTION:
WHEELOCK CREEK 28.0
END DESCRIPTION:
XS GIS Cut Line= 3
      3670849.64     10514960.18      3672449.61     10514610.19
       3673149.6     10514360.19
#Sta/Elev= 30
  3369.9   294.4  3580.1  285.81  3858.7   257.3  4649.4  256.03  4905.7  258.12
  4966.8  258.83  4983.2   251.2  4988.3  254.19  4994.5  250.06  4997.2  249.56
  5000.5  250.06  5005.1  252.64  5010.4  252.64  5017.8  259.02  5023.1  256.54
  5028.9  259.24  5060.9  258.72  5220.1   256.8  5314.6  264.86  5326.3  267.38
  5438.3  274.97  5499.9  281.65  5530.7  286.41  5549.3  293.22  5556.2  298.35
  5581.1  303.33  5623.6  309.74  5713.2  318.63  5736.4  321.11    5751  322.15
#Mann= 8 ,-1 , 0
  3369.9     .05       0  4905.7     .16       0  4994.5     .07       0
  5000.5     .16       0  5060.9     .05       0  5314.6      .1       0
  5713.2     .16       0  5736.4      .1       0
Bank Sta=4966.8,5017.8
XS Rating Curve= 0 ,0
Exp/Cntr=0.3,0.1

Type RM Length L Ch R = 1 ,17657   ,552,552,552
BEGIN DESCRIPTION:
WHEELOCK CREEK 27.0
END DESCRIPTION:
XS GIS Cut Line= 3
      3671049.59     10514960.19      3672649.61     10515060.19
      3673449.65     10514960.18
#Sta/Elev= 30
  3482.2  290.99  3564.9  284.53  3720.2  262.81  3782.8  257.49  4554.3  254.39
  4872.1  255.23  4965.1  257.35  4975.1  252.99  4992.2  248.53  4994.9  248.03
  4998.2  248.53  5007.7  248.84  5015.2  256.63  5091.9  257.53  5246.6  256.34
  5276.8  254.89  5397.7  262.65  5550.4  277.71  5619.5  285.69  5669.9  297.39
  5687.5  304.38  5692.5  302.92  5710.2  309.59  5730.3  314.67  5750.5  317.34
  5768.1  321.62  5773.1  321.42  5780.7   324.3  5841.2  333.39  5891.6  338.26
#Mann= 6 ,-1 , 0
  3482.2     .05       0  4872.1     .16       0  4992.2     .07       0
  4998.2     .16       0  5091.9     .05       0  5550.4      .1       0
Bank Sta=4965.1,5015.2
XS Rating Curve= 0 ,0
Exp/Cntr=0.3,0.1

Type RM Length L Ch R = 1 ,17105   ,342,342,342
BEGIN DESCRIPTION:
WHEELOCK CREEK 26.0
END DESCRIPTION:
XS GIS Cut Line= 3
      3670449.56     10515560.19      3672849.61     10515360.19
      3673249.63     10515410.19
#Sta/Elev= 30
    2591   326.9  3032.6  310.61  3092.8  304.58  3112.9  300.13  3243.3  284.64
  3255.8  281.24  3376.3  267.96  3474.1  261.66  3644.7  258.03  4235.2  254.38
  4296.8  252.73    4327  254.56  4502.1  253.52  4868.9  256.29  4989.3  255.17
  4992.9  251.57  4996.9  247.58  5006.4  247.55  5009.2  247.05  5012.4  247.55
  5029.6  255.66  5100.1  255.48    5211  266.36  5251.3  274.17    5275  284.75
    5279  288.06  5291.6  290.31  5331.9   304.9    5384  314.07  5402.5  316.29
#Mann= 9 ,-1 , 0
    2591     .05       0  4235.2     .16       0  4296.8     .12       0
  4502.1     .16       0  4992.9     .05       0  5006.4     .03       0
  5012.4     .05       0    5275     .16       0    5384      .1       0
Bank Sta=4989.3,5029.6
XS Rating Curve= 0 ,0
Exp/Cntr=0.3,0.1

Type RM Length L Ch R = 1 ,16763   ,866,866,866
BEGIN DESCRIPTION:
WHEELOCK CREEK 25.0
END DESCRIPTION:
XS GIS Cut Line= 3
      3670549.64     10515660.19      3673018.86     10515670.36
      3673199.57     10515510.22
#Sta/Elev= 30
  2643.5  326.11  3033.5  311.09  3313.5  277.18  3443.5  266.18  3583.5   261.5
  3733.5   262.8  3881.1  259.23  4413.5  252.07  4843.5  252.23  4983.5  254.81
  5003.5  247.32  5010.5  247.19  5013.2  246.69  5016.5  247.19  5023.5     252
  5033.5  255.02  5040.2  254.94  5083.5  253.38  5155.6  260.09  5191.6  268.78
  5198.3  268.02  5226.7  273.75    5234  279.29  5247.6   282.9  5255.1  287.79
    5276  293.29  5282.9  297.35  5290.3  296.32  5297.8  301.19  5354.2  310.62
#Mann= 6 ,-1 , 0
  2643.5     .05       0  3881.1     .16       0  5010.5     .07       0
  5016.5     .16       0  5040.2     .05       0  5282.9      .1       0
Bank Sta=4983.5,5033.5
XS Rating Curve= 0 ,0
Exp/Cntr=0.3,0.1

Type RM Length L Ch R = 1 ,15897   ,684,684,684
BEGIN DESCRIPTION:
WHEELOCK CREEK 24.0
END DESCRIPTION:
XS GIS Cut Line= 3
      3671749.62     10516560.19      3673199.61     10516210.19
      3673249.61     10515460.19
#Sta/Elev= 30
  3479.4  303.49    3572  297.98  3746.9  284.03  3801.2   278.7  3935.3  261.36
  3968.8  256.97  4094.4  251.09  4139.9  250.48  4345.3  250.27    4448  249.82
  4907.3   253.6  4952.7   252.5  4978.1  245.84  4980.8  245.34  4984.1  245.84
  5011.1  248.63  5046.2  248.66  5051.2     251  5072.7  251.71  5081.3  253.34
  5201.5  252.25  5300.5  260.31    5392  268.53  5432.1  268.34  5462.1  276.55
  5472.1   277.1  5512.2  289.31  5552.3  297.17  5662.6  312.31  5722.7   317.6
#Mann= 10 ,-1 , 0
  3479.4     .05       0  3935.3     .16       0  4139.9     .12       0
  4345.3     .16       0    4448     .05       0  4907.3     .16       0
  4978.1     .07       0  4984.1     .16       0  5072.7     .05       0
  5300.5      .1       0
Bank Sta=4952.7,5081.3
XS Rating Curve= 0 ,0
Exp/Cntr=0.3,0.1

Type RM Length L Ch R = 1 ,15213   ,719,719,719
BEGIN DESCRIPTION:
WHEELOCK CREEK 23.0
END DESCRIPTION:
XS GIS Cut Line= 3
      3672349.64     10517460.16      3673649.61     10516360.19
      3673999.61      10515560.2
#Sta/Elev= 30
  3311.6  302.52  3431.8   296.7  3503.3  289.32  3559.8   278.4  3609.9  271.81
  3638.5  265.35  3680.1  260.76  3702.2  261.34    3780  252.55  3829.6  248.12
  3884.6  247.55  4063.4  247.95  4297.6  249.11  4489.9  246.68  4897.9  251.16
  4978.8  251.56  4983.5  244.38  4986.3  243.88  4989.5  244.38  5000.8  244.63
  5011.2  250.23  5023.5  251.34  5179.3  249.89  5365.1  250.08  5447.4  254.17
  5723.1  273.01  5750.9  274.16  5797.7  280.58  5855.4  301.73  5887.7  308.69
#Mann= 12 ,-1 , 0
  3311.6     .05       0  3559.8     .16       0    3780     .05       0
  3884.6     .07       0  4063.4     .05       0  4897.9     .16       0
  4983.5     .07       0  4989.5     .16       0  5179.3     .05       0
  5365.1     .16       0  5447.4     .05       0  5723.1     .16       0
Bank Sta=4978.8,5023.5
XS Rating Curve= 0 ,0
Exp/Cntr=0.3,0.1

Type RM Length L Ch R = 1 ,14494   ,611,611,611
BEGIN DESCRIPTION:
WHEELOCK CREEK 22.0
END DESCRIPTION:
XS GIS Cut Line= 3
       3672449.6     10517510.19      3673899.61     10516710.19
      3674399.65     10516410.17
#Sta/Elev= 30
  3335.5  300.82  3403.1  297.79  3494.1  288.28  3586.8  273.09  3666.7  263.93
  3674.8  265.68  3712.4   255.3  3794.8  248.13  3910.2  247.46  4637.5  245.99
  4948.7  249.63  4961.8  249.96  4985.7  243.11  4988.5  242.61  4991.7  243.11
  4999.3  246.72  5005.2  244.21  5042.1  245.19  5057.6   249.4  5063.5   244.7
  5095.3  250.66  5165.7  248.56  5341.4  257.84    5493  273.69  5516.3  278.06
  5524.1  282.63    5530  279.95    5561  285.51  5566.9  281.71  5574.7  282.92
#Mann= 9 ,-1 , 0
  3335.5     .05       0  3494.1     .16       0  3794.8     .12       0
  3910.2     .05       0  4948.7     .16       0  4985.7     .07       0
  4991.7     .16       0  5095.3     .05       0  5165.7     .16       0
Bank Sta=4961.8,5057.6
XS Rating Curve= 0 ,0
Exp/Cntr=0.3,0.1

Type RM Length L Ch R = 1 ,13883   ,535,535,535
BEGIN DESCRIPTION:
WHEELOCK CREEK 21.0
END DESCRIPTION:
XS GIS Cut Line= 3
      3672699.62     10517660.19      3673906.02     10517227.65
       3674799.6      10516310.2
#Sta/Elev= 30
  3711.9  296.18  3807.5  288.86    3845  284.44  3881.9  275.61  3924.4  271.36
  3998.7  260.14  4073.1  252.75  4080.3  250.65  4141.8     246  4220.9  245.63
    4328  245.98  4354.4  244.26  4370.5  245.85  4464.1  244.52  4806.1  246.13
  4954.4  248.99  4986.7  248.93  5005.4  243.05  5008.1  242.55  5011.4  243.05
  5029.7  249.05  5036.6  248.97  5046.8  248.98  5087.5   248.9  5397.3  247.28
  5524.6  252.34  5545.9  255.18  5662.8  255.44  5970.1  260.06  6274.2  271.37
#Mann= 9 ,-1 , 0
  3711.9     .16       0  4220.9     .12       0  4354.4     .05       0
  4954.4     .16       0  5005.4     .07       0  5011.4     .16       0
  5046.8     .12       0  5087.5     .05       0  5662.8     .16       0
Bank Sta=4986.7,5036.6
XS Rating Curve= 0 ,0
Exp/Cntr=0.3,0.1

Type RM Length L Ch R = 1 ,13348   ,649,649,649
BEGIN DESCRIPTION:
WHEELOCK CREEK 20.0
END DESCRIPTION:
XS GIS Cut Line= 3
      3672699.64     10517760.18      3674149.61     10517560.19
      3675099.62     10515960.16
#Sta/Elev= 30
  3520.3  298.81  3651.5  293.29    3872  265.35  4159.9  248.03  4258.2  243.79
  4960.6  247.76  4973.9  247.78  4994.6  242.13  4997.4  241.63  5000.6  242.13
    5019  247.59  5087.3  244.45  5093.1  248.18  5134.3  248.02  5757.5  249.37
  6028.4  260.78  6195.3  262.53  6283.6  259.58  6289.4  265.17  6305.1  262.05
  6326.5  266.54  6342.1  261.28  6347.9  267.12  6363.5  263.41  6369.3  270.53
  6379.1  272.71    6459  270.85  6603.1  288.07  6735.7  316.21  6844.8  327.07
#Mann= 9 ,-1 , 0
  3520.3     .16       0    3872     .05       0  4159.9     .16       0
  4258.2     .05       0  4960.6     .07       0  4994.6     .07       0
  5000.6     .07       0  5134.3     .05       0  6195.3     .16       0
Bank Sta=4973.9,5019
XS Rating Curve= 0 ,0
Exp/Cntr=0.3,0.1

Type RM Length L Ch R = 1 ,12699   ,512,512,512
BEGIN DESCRIPTION:
WHEELOCK CREEK 19.0
END DESCRIPTION:
XS GIS Cut Line= 3
       3672799.6     10517810.19      3674399.61     10517910.19
      3675949.64     10516760.16
#Sta/Elev= 30
  3394.2  297.17  3592.4  273.66  3714.8  262.84  3865.1  256.89  3905.2   251.8
    4029  243.58  4095.6  241.64  4187.6  243.19  4875.1  244.83  4967.3  246.06
  4987.3  244.02  4991.8  240.91  4994.6  240.41  4997.8  240.91  5004.6   244.8
  5010.9  242.37  5019.3  245.98  5148.9  244.32  5440.7  242.36  6127.2  247.51
    6269  251.81  6393.9  265.51  6548.7  287.96  6584.1  295.28    6641  310.56
  6648.8  315.43  6705.1  329.71    6749  339.32  6784.9  343.83  6927.4  345.87
#Mann= 10 ,-1 , 0
  3394.2     .16       0  3592.4     .05       0    4029     .16       0
  4187.6     .05       0  4875.1     .12       0  4991.8     .07       0
  4997.8     .12       0  5148.9     .05       0  6393.9     .16       0
  6784.9     .05       0
Bank Sta=4967.3,5019.3
XS Rating Curve= 0 ,0
Exp/Cntr=0.3,0.1

Type RM Length L Ch R = 1 ,12187   ,774,774,774
BEGIN DESCRIPTION:
WHEELOCK CREEK 18.0
END DESCRIPTION:
XS GIS Cut Line= 4
      3672812.24     10518889.12       3674333.1     10518295.36
      3674973.72     10518154.74       3676124.7     10517071.47
#Sta/Elev= 30
  2974.8  302.51  2976.6  302.39  3090.1   296.8  3186.7  282.21  3433.6   256.1
  3812.3  244.31  4009.9  241.99  4027.8  242.15  4183.6  240.45  4514.8  239.85
  4517.6  239.35  4520.8  239.85  4559.3  241.57  4684.6  241.61  4977.2  244.98
  4979.5  245.02  5003.2  240.07  5033.9  244.91  5079.3  246.73  5085.1  248.14
  5105.5  241.91  5574.7   249.5  6098.3  247.39  6260.9   252.3  6370.6  262.19
  6544.2  282.24  6692.6  322.57  6706.8  330.93  6780.2  338.46  6843.9  338.22
#Mann= 14 ,-1 , 0
  2974.8     .05       0  2976.6     .16       0  3812.3     .12       0
  4009.9     .05       0  4027.8     .12       0  4183.6     .05       0
  4514.8     .07       0  4520.8     .05       0  4559.3     .12       0
  4684.6     .05       0  4977.2     .12       0  5079.3     .05       0
  6370.6     .16       0  6780.2     .05       0
Bank Sta=4979.5,5033.9
XS Rating Curve= 0 ,0
Exp/Cntr=0.3,0.1

Type RM Length L Ch R = 1 ,11413   ,591,591,591
BEGIN DESCRIPTION:
WHEELOCK CREEK 17.0
END DESCRIPTION:
XS GIS Cut Line= 3
      3672899.57      10519110.2      3674899.61     10518710.19
      3676083.09     10518951.61
#Sta/Elev= 30
  2949.2  303.48  3013.4  302.18  3204.2  290.56  3285.8   277.2  3416.1  263.02
  3591.7  245.93  3683.5  244.45  3775.3  238.56  4210.8  238.37  4213.5  237.87
  4216.8  238.37  4554.9  239.16  4758.1  240.62  4948.1  243.45  4968.5  239.12
  5029.7   242.6  5356.3   243.4  5458.3  249.27  5564.8   259.9    5591  258.22
  5703.3  276.42  5711.3  281.49    5767   295.9  5784.9  304.72    5887  325.74
  5918.6  328.37  6009.4  327.55  6014.5  330.35  6115.6  341.35  6196.7  342.98
#Mann= 8 ,-1 , 0
  2949.2     .05       0  3013.4     .16       0  3416.1     .05       0
  4210.8     .03       0  4216.8     .05       0  4554.9     .16       0
  4758.1     .05       0    5591     .16       0
Bank Sta=4948.1,5029.7
XS Rating Curve= 0 ,0
Exp/Cntr=0.3,0.1

Type RM Length L Ch R = 1 ,10822   ,608,608,608
BEGIN DESCRIPTION:
WHEELOCK CREEK 16.0
END DESCRIPTION:
XS GIS Cut Line= 3
      3673349.64     10519060.19      3674949.61     10519160.19
      3675649.59     10519510.18
#Sta/Elev= 30
  3415.4  266.26  3425.4  266.24  3439.5  262.89  3653.3  245.52  3796.1  240.68
  4036.6  241.51  4156.8  238.29  4327.1   239.8  4427.1  237.62  4467.4  239.08
  4848.2  238.25  4988.4   241.8  4998.5  239.88  5008.5  241.88    5016  242.38
  5074.9  241.83  5121.9  240.42    5175  242.74  5197.4  245.96  5390.2  259.72
  5563.5  278.72  5622.2  292.45  5644.6  299.46    5653  303.79  5680.9  309.31
  5711.7  319.87  5725.7  321.51  5742.4  328.63  5787.1  337.58  5801.1  338.53
#Mann= 5 ,-1 , 0
  3415.4     .16       0  3439.5     .05       0  4988.4     .03       0
  5008.5     .05       0  5074.9     .16       0
Bank Sta=4988.4,5016
XS Rating Curve= 0 ,0
Exp/Cntr=0.3,0.1

Type RM Length L Ch R = 1 ,10214   ,557,557,557
BEGIN DESCRIPTION:
WHEELOCK CREEK 15.0
END DESCRIPTION:
XS GIS Cut Line= 3
      3673299.61     10519210.19      3674899.61     10519610.19
      3675599.59     10519560.19
#Sta/Elev= 30
  3334.6  278.91  3386.1  272.48  3406.7  273.38    3448  267.28  3483.1  265.08
  3551.1  260.98    3600  254.72  3646.4  253.64  3723.7  246.71  3839.7  240.76
  4676.9  237.62  4993.9  240.44  5003.9  238.95  5023.9  241.12  5084.1  240.37
  5134.2  239.51  5196.9  242.98    5435  270.24  5465.1  276.14  5472.6  279.89
  5477.6  277.92  5495.1   284.9  5505.2  286.29  5555.3  302.47  5605.4  314.56
  5612.9  318.69    5618  317.42  5645.5  323.16  5675.6  332.86  5685.6  334.07
#Mann= 5 ,-1 , 0
  3334.6     .16       0  3483.1     .05       0  5003.9     .03       0
  5023.9     .05       0  5084.1     .16       0
Bank Sta=4993.9,5023.9
XS Rating Curve= 0 ,0
Exp/Cntr=0.3,0.1

Type RM Length L Ch R = 1 ,9657    ,573,573,573
BEGIN DESCRIPTION:
WHEELOCK CREEK 14.0
END DESCRIPTION:
XS GIS Cut Line= 3
      3673049.65      10519410.2      3674649.61     10519960.19
       3675449.6     10520010.19
#Sta/Elev= 30
  3307.3  303.46  3354.1  302.01  3416.6  296.45  3518.7  278.09  3598.8  266.55
  3604.1  267.95  3635.3  262.45    3656  262.69  3666.8  259.36  3781.7   249.8
  3874.7  244.76  4025.6  241.87  4322.4  242.82  4525.5  238.09  4935.7  238.21
  4983.5  239.79  5006.2  237.05  5008.9  236.55  5012.2  237.05  5019.2  239.98
  5242.1  239.09  5530.2  254.92  5540.2  255.05  5569.3   248.7  5580.3  249.35
  5600.3  256.61  5630.4  259.55  5660.4  266.63  5710.5  273.05  5800.7  291.85
#Mann= 5 ,-1 , 0
  3307.3     .16       0  3781.7     .16       0  5006.2     .03       0
  5012.2     .16       0  5569.3     .16       0
Bank Sta=4983.5,5019.2
XS Rating Curve= 0 ,0
Exp/Cntr=0.3,0.1
