HEC-RAS study BIG BROWN CREEK.prj: BIG BROWN CREEK Base Level Engineering

--- BIG BROWN CREEK.g01 (geometry) --- (continued)

Type RM Length L Ch R = 1 ,44908   ,568,568,568
BEGIN DESCRIPTION:
BIG BROWN CREEK 59.0
END DESCRIPTION:
XS GIS Cut Line= 3
      3617949.57     10634860.19      3618499.61     10634810.19
      3620049.63     10633210.17
#Sta/Elev= 30
  4446.3  333.05  4466.4   332.5  4516.6  326.62  4546.7  324.28  4556.8  321.95
  4566.8  321.35  4647.2  310.98  4657.2  310.27  4677.3   311.1  4697.4  309.03
  4704.4  303.61  4707.2  303.11  4710.4  303.61  4724.2  303.61    6517  303.61
  6526.7  303.61  6582.8  303.61  6589.7  309.36  6596.9  309.63  6611.1  309.53
  6665.2  312.65  6681.8  312.81  6745.4   317.9  6789.8  319.91    6908  326.22
  6922.1  327.98  7027.1   334.7  7084.9  337.88  7219.8  348.56  7226.3  348.81
#Mann= 10 ,-1 , 0
  4446.3     .16       0  4704.4    .033       0  4710.4     .16       0
  4724.2     .05       0    6517     .07       0  6526.7     .12       0
  6665.2     .16       0  6789.8     .12       0  7027.1     .16       0
  7219.8     .12       0
Bank Sta=4677.3,6596.9
XS Rating Curve= 0 ,0
Exp/Cntr=0.3,0.1

Type RM Length L Ch R = 1 ,44340   ,512,512,512
BEGIN DESCRIPTION:
BIG BROWN CREEK 58.0
END DESCRIPTION:
XS GIS Cut Line= 3
      3617799.59     10635610.19      3618599.61     10635360.19
      3620149.61     10635110.19
#Sta/Elev= 30
    4187  340.19  4203.3  337.37  4228.9  335.92  4235.7  333.79  4305.9  327.69
  4312.7  326.12  4338.4  324.77  4370.9  320.41  4490.8  313.44  4522.3  309.94
  4538.5  310.65  4576.2  309.63  4582.1  303.61  4584.9  303.11  4588.1  303.61
  4607.5  303.61  6136.5  303.61  6139.4  303.61  6149.5  309.73  6179.9  311.06
    6191   310.1  6237.3  313.52  6252.8  313.77  6338.2  320.99  6376.4  322.28
  6402.7  325.28    6439  327.63    6500  334.34  6566.8  338.34  6595.2   341.4
#Mann= 8 ,-1 , 0
    4187     .16       0  4582.1    .033       0  4588.1     .16       0
  4607.5     .05       0  6136.5     .16       0  6237.3     .12       0
  6338.2     .16       0    6439     .12       0
Bank Sta=4538.5,6179.9
XS Rating Curve= 0 ,0
Exp/Cntr=0.3,0.1

Type RM Length L Ch R = 1 ,43828   ,547,547,547
BEGIN DESCRIPTION:
BIG BROWN CREEK 57.0
END DESCRIPTION:
XS GIS Cut Line= 3
      3618249.61     10636260.18      3618799.61     10635810.19
      3620349.64     10635110.17
#Sta/Elev= 30
  4324.7  334.97    4370  331.91  4438.8  326.12  4445.3  323.03    4474  322.27
  4488.4  320.21  4552.2  316.31  4558.7  314.78  4616.1  310.52  4644.8  310.79
  4651.3  309.44  4656.2  303.61  4658.9  303.11  4662.2  303.61  4679.2  303.61
  5995.2  303.61  6000.9   309.7    6010  309.59  6041.5   311.1  6055.8   310.6
    6231  320.66  6289.1  323.91  6341.1  328.85  6508.2  340.23  6606.2  350.34
  6623.8  353.39  6629.3  352.87  6675.5  356.68  6698.6  361.05  6736.1  362.69
#Mann= 7 ,-1 , 0
  4324.7     .12       0    4370     .16       0  4656.2    .033       0
  4662.2     .16       0  4679.2     .05       0    6010     .16       0
    6231     .12       0
Bank Sta=4644.8,6041.5
XS Rating Curve= 0 ,0
Exp/Cntr=0.3,0.1

Type RM Length L Ch R = 1 ,43281   ,540,540,540
BEGIN DESCRIPTION:
BIG BROWN CREEK 56.0
END DESCRIPTION:
XS GIS Cut Line= 3
      3618399.58      10636460.2      3619099.61     10636260.19
      3620499.62     10636010.19
#Sta/Elev= 30
  4271.6  337.28  4313.2  335.48  4322.3  333.72    4334  333.34  4434.1  321.46
  4448.4  321.27  4458.8  319.45  4473.1  319.12  4479.6  317.62  4521.2  314.09
  4573.2  310.19  4618.7  310.23  4625.2  309.62  4635.6  305.07    4643  303.61
  4645.8  303.11    4649  303.61  4653.8  303.61    5871  303.61  5873.2  303.61
  5879.9  309.78  5913.9  311.05  5944.4  310.85  6026.6   315.8  6164.3  330.09
  6223.2   334.5  6282.1  340.34  6289.7  342.17  6360.8  350.54  6421.8   355.8
#Mann= 6 ,-1 , 0
  4271.6     .16       0    4643    .033       0    4649     .16       0
  4653.8     .05       0    5871     .16       0  6026.6     .12       0
Bank Sta=4618.7,5913.9
XS Rating Curve= 0 ,0
Exp/Cntr=0.3,0.1

Type RM Length L Ch R = 1 ,42741   ,217,217,217
BEGIN DESCRIPTION:
BIG BROWN CREEK 55.0
END DESCRIPTION:
XS GIS Cut Line= 3
       3618499.6     10636610.19      3619299.61     10636760.19
      3620549.61     10636060.19
#Sta/Elev= 30
  4184.8  329.76  4215.5     328    4256   323.5  4286.5   322.1  4316.2  318.17
  4321.3  319.06  4337.4  317.08  4357.8  316.81  4367.9  315.79  4373.9  313.88
  4408.6  312.43  4418.8  310.45  4484.1   310.9  4500.2  309.48  4507.4  303.61
  4510.1  303.11  5858.3  303.61  5872.1  309.82  5909.7  310.64  5925.7  309.74
  5947.4  313.19  6012.5  317.59  6158.6  330.67    6248  339.23  6277.3  343.89
    6299  345.13  6305.3  346.65  6364.1  352.63  6401.7  354.65  6431.4  354.13
#Mann= 4 ,-1 , 0
  4184.8     .12       0  4215.5     .16       0  4484.1     .07       0
  5909.7     .12       0
Bank Sta=4484.1,5909.7
XS Rating Curve= 0 ,0
Exp/Cntr=0.3,0.1

Type RM Length L Ch R = 1 ,42524   ,792,792,792
BEGIN DESCRIPTION:
BIG BROWN CREEK 54.0
END DESCRIPTION:
XS GIS Cut Line= 2
      3616911.08     10638568.59      3620869.45     10635999.12
#Sta/Elev= 30
  2021.2  372.39  2135.2  370.57  2307.2  362.37  2479.7  356.71  2778.5  345.68
  2959.7  345.37  3270.8  336.14  3414.3  327.16    3458  326.03  3587.9  316.88
  3738.9  310.65  3790.2  310.72  3817.8  310.11  3819.7  310.11  3823.5  303.61
  3826.2  303.11  3829.5  303.61  5886.3  303.61  5894.1  309.44  5929.9  309.54
  5937.7  312.69    5993  316.85  6227.7  336.48  6327.2  347.76  6363.5  348.53
  6378.6  346.67  6466.3  344.67  6559.9  349.64  6674.6  359.31  6740.4  358.96
#Mann= 6 ,-1 , 0
  2021.2     .05       0  2479.7     .16       0  3817.8     .05       0
  3823.5    .033       0  3829.5     .05       0    5993     .12       0
Bank Sta=3790.2,5894.1
XS Rating Curve= 0 ,0
Exp/Cntr=0.3,0.1

Type RM Length L Ch R = 1 ,41732   ,607,607,607
BEGIN DESCRIPTION:
BIG BROWN CREEK 53.0
END DESCRIPTION:
XS GIS Cut Line= 2
       3617362.5     10639280.37      3621043.08     10636576.36
#Sta/Elev= 30
  2297.5  381.53  2875.7  342.47  2988.8  340.64  3017.7  338.49  3032.4  331.41
  3038.6  337.66    3047  331.97  3053.2  335.97  3075.7   329.9  3097.2  335.18
  3283.1  324.25  3404.3  324.44  3611.1  310.76  3733.3  309.57  3737.7  303.61
  3740.5  303.11  3743.7  303.61  3815.7  303.61    3973  303.61  4063.8  303.61
  4130.3  303.61  4226.1  303.61  4306.4  303.61  6358.8  303.61    6365  311.31
  6489.2  320.07    6674  335.06  6718.1  339.56  6803.7  347.98  6864.6  349.75
#Mann= 13 ,-1 , 0
  2297.5     .16       0  3737.7    .033       0  3743.7     .16       0
  3815.7     .07       0    3973     .05       0  4063.8     .07       0
  4130.3     .05       0  4226.1     .07       0  4306.4     .05       0
  6489.2     .16       0    6674     .12       0  6718.1     .16       0
  6803.7     .12       0
Bank Sta=3611.1,6365
XS Rating Curve= 0 ,0
Exp/Cntr=0.3,0.1

Type RM Length L Ch R = 1 ,41125   ,1118,1118,1118
BEGIN DESCRIPTION:
BIG BROWN CREEK 52.0
END DESCRIPTION:
XS GIS Cut Line= 3
      3617523.09     10639513.08      3619849.61     10638210.19
      3621099.61     10636610.18
#Sta/Elev= 30
  2316.5  365.09    2910  340.98  2941.9  332.55  2963.6  331.17  2985.3  334.59
    2991   331.4  3028.7   331.4  3109.7   335.9  3396.2  333.71  3859.8  318.33
  3953.3  314.66  3969.3  311.22  4089.6  309.47  4137.1  309.26  4143.3  303.61
  4146.1  303.11  4149.3  303.61  4193.3  303.61  6521.4  303.61  6529.5  309.11
  6579.3  318.22  6643.3  322.05  6856.9  343.88  6877.7  343.29  6884.8  346.67
  6887.6  346.29  6892.2  343.87  6906.7  349.57  7005.6  355.28  7013.4  354.96
#Mann= 9 ,-1 , 0
  2316.5     .16       0  4089.6     .07       0  4143.3    .033       0
  4149.3     .07       0  4193.3     .05       0  6643.3      .1       0
  6884.8     .16       0  6887.6      .1       0  7005.6     .12       0
Bank Sta=3859.8,6579.3
XS Rating Curve= 0 ,0
Exp/Cntr=0.3,0.1

Type RM Length L Ch R = 1 ,40007   ,977,977,977
BEGIN DESCRIPTION:
BIG BROWN CREEK 50.0
END DESCRIPTION:
XS GIS Cut Line= 4
      3618278.24      10639374.2      3620305.21     10639223.95
      3620630.73     10639050.34      3621509.62     10636598.13
#Sta/Elev= 30
  2820.9  348.97  2882.4  344.75  3022.8  339.77  3378.2  333.33  3565.8  331.49
    3635   331.6  3744.8  325.62  3794.9  319.54  3875.1  313.39    3885  310.11
  3905.2  310.92  3945.3  309.69  3952.4  303.61  3955.1  303.11  3958.4  303.61
  3978.8  303.61  7222.3  303.61  7247.7  313.96  7262.9  314.64  7325.8  319.57
  7389.6  327.59  7483.1  334.95  7544.7  341.25  7693.1  349.34  7698.4  347.86
  7749.3  349.95  7754.6   348.5  7810.8  350.64  7816.1  349.22  7827.3  349.63
#Mann= 9 ,-1 , 0
  2820.9     .16       0  3378.2     .12       0  3565.8     .16       0
    3635     .12       0  3952.4    .033       0  3958.4     .12       0
  3978.8     .05       0  7262.9     .16       0  7483.1     .12       0
Bank Sta=3905.2,7247.7
XS Rating Curve= 0 ,0
Exp/Cntr=0.3,0.1

Type RM Length L Ch R = 1 ,39030   ,103,103,103
BEGIN DESCRIPTION:
BIG BROWN CREEK 49.0
END DESCRIPTION:
XS GIS Cut Line= 4
       3617783.5     10639608.58      3620543.92     10640146.26
      3620934.55     10640016.05      3621997.91     10636717.46
#Sta/Elev= 30
  1990.1  355.82  2383.5  350.12  2549.6   352.1    2954  325.96  2967.7  321.94
  2984.5   323.4  3004.9  318.61  3035.5  323.95  3218.9  327.36  3402.3  319.09
  3473.6  319.37    3606  310.39  3626.4  311.24  3632.6  310.56  3643.9  309.72
    3654  303.61  3656.7  303.11    3660  303.61  8120.3  303.61  8130.7  309.94
  8141.2  312.17  8179.1  314.13  8239.5  320.84  8351.3  322.93  8362.2  326.23
    8443  333.94  8544.7  340.59  8601.1  344.09    8614  349.06  8679.9  355.43
#Mann= 8 ,-1 , 0
  1990.1     .16       0  3632.6     .05       0    3654    .033       0
    3660     .05       0  8239.5      .1       0  8362.2     .08       0
    8443     .05       0  8544.7     .08       0
Bank Sta=3626.4,8179.1
XS Rating Curve= 0 ,0
Exp/Cntr=0.3,0.1

Type RM Length L Ch R = 1 ,38927   ,451,451,451
BEGIN DESCRIPTION:
BIG BROWN CREEK 48.0
END DESCRIPTION:
XS GIS Cut Line= 3
      3620049.61     10641660.18      3620509.63     10640261.06
      3624749.63     10638910.18
#Sta/Elev= 30
  3243.7  329.07  3285.8  327.32  3291.4  326.45  3306.9  326.31  3317.4  324.45
  3323.2  324.64  3328.5  323.84  3338.4  324.65  3386.8  321.87  3506.9  316.27
    3514   315.3  3519.2  315.28  3527.9  313.29  3534.3   312.5  3545.8  310.65
  3557.9  310.74  3591.1  309.82  3606.4  303.61  3609.1  303.11  3612.4  303.61
  3623.7  303.61  9009.1  303.61  9016.3  306.52  9021.5  309.75    9030  310.33
  9040.5  312.79  9053.7   313.6  9061.5  315.08  9109.1  318.57  9166.5   322.9
#Mann= 7 ,-1 , 0
  3243.7     .12       0  3534.3     .05       0  3557.9     .12       0
  3606.4    .033       0  3612.4     .12       0  3623.7     .05       0
  9109.1     .16       0
Bank Sta=3557.9,9030
XS Rating Curve= 0 ,0
Exp/Cntr=0.3,0.1

Type RM Length L Ch R = 1 ,38476   ,690,690,690
BEGIN DESCRIPTION:
BIG BROWN CREEK 47.0
END DESCRIPTION:
XS GIS Cut Line= 3
      3620149.59     10641810.22      3620999.61     10640560.19
      3624999.62     10638960.19
#Sta/Elev= 30
    3504     335  3612.9   330.8  3706.1  325.05    3727  324.51  3733.8   323.1
  3842.6  315.07  3864.7  310.64  3885.7  310.67  3915.2  309.61  3918.6  303.61
  3921.4  303.11  3924.6  303.61  3929.4  303.61  8925.3  303.61    8932   309.5
  8937.4  309.68  8946.8  313.42  8961.6  313.36  8989.1  315.41  9102.5  323.17
  9117.8  325.45  9123.2  324.02  9140.7  325.35  9147.4   326.7  9230.9  329.88
  9255.1   332.3  9302.3  334.68    9309  335.67  9314.4     335  9323.8  335.81
#Mann= 6 ,-1 , 0
    3504     .12       0  3918.6    .033       0  3924.6     .12       0
  3929.4     .05       0  8989.1     .16       0  9102.5     .12       0
Bank Sta=3885.7,8946.8
XS Rating Curve= 0 ,0
Exp/Cntr=0.3,0.1

Type RM Length L Ch R = 1 ,37786   ,373,373,373
BEGIN DESCRIPTION:
BIG BROWN CREEK 46.0
END DESCRIPTION:
XS GIS Cut Line= 3
      3620649.62     10642560.16      3621095.57     10641302.73
       3625199.6      10639010.2
#Sta/Elev= 30
  3420.6  341.53  3492.5  336.23  3528.6   335.8  3585.1  331.09  3605.3     331
  3646.8   329.9  3826.8  318.69  3852.3  315.78  3888.5  314.79    3898  310.82
  3909.2  310.63  3914.1  310.71  3951.1  310.09  3961.7  307.27  3967.5  303.61
  3970.3  303.11  3973.5  303.61  4014.8  303.61  8837.2  303.61  8846.9  309.54
  8850.3  309.55    8896   311.1  8988.9  319.03  9014.8  321.49  9020.5  323.24
  9036.5  323.61  9052.5  326.16  9101.6  330.13    9177  331.06  9455.7  345.44
#Mann= 8 ,-1 , 0
  3420.6     .16       0  3605.3     .12       0  3909.2     .16       0
  3967.5    .033       0  3973.5     .16       0  4014.8     .05       0
  8850.3     .16       0  8988.9     .12       0
Bank Sta=3914.1,8896
XS Rating Curve= 0 ,0
Exp/Cntr=0.3,0.1

Type RM Length L Ch R = 1 ,37413   ,480,480,480
BEGIN DESCRIPTION:
BIG BROWN CREEK 45.0
END DESCRIPTION:
XS GIS Cut Line= 3
      3620849.59     10642410.22      3621549.61     10641460.19
      3625149.59     10640260.19
#Sta/Elev= 30
  3845.7   337.4  3953.3  330.33  4060.5  319.75  4118.3  315.42  4139.2   311.6
  4168.5   310.1  4181.1  309.72  4189.3  306.74  4192.5  303.61  4195.3  303.11
  4198.5  303.61  4222.4  303.61  7334.2  303.61  7344.8  305.16  7355.3  309.66
  7376.4  310.37    7408  314.63  7434.1  316.17  7492.4  321.79  7530.3  321.75
  7734.8  320.48  8124.8  331.88  8198.6  332.74  8314.6  328.52  8386.5  321.98
  8398.1  319.66  8409.4  317.65  8525.4  328.57    8702   338.6  8820.5  340.14
#Mann= 10 ,-1 , 0
  3845.7     .12       0  4060.5     .16       0  4192.5    .033       0
  4198.5     .16       0  4222.4     .05       0  7434.1     .16       0
  7530.3     .12       0  8386.5     .16       0  8398.1     .12       0
    8702     .05       0
Bank Sta=4168.5,7376.4
XS Rating Curve= 0 ,0
Exp/Cntr=0.3,0.1

Type RM Length L Ch R = 1 ,36933   ,515,515,515
BEGIN DESCRIPTION:
BIG BROWN CREEK 44.0
END DESCRIPTION:
XS GIS Cut Line= 3
      3621049.59     10642560.21      3621749.61     10641910.19
      3624149.65     10640710.17
#Sta/Elev= 30
  4037.7  335.55  4136.7  328.03    4250  321.43  4313.5  316.67  4320.9  315.56
  4327.7  312.28  4363.4  311.16  4375.5  309.97  4398.6  309.61  4401.6  305.42
  4402.9  303.61  4405.7  303.11  4408.9  303.61  7265.4  303.61  7273.8  309.51
  7287.7  309.76  7316.2   314.2  7326.9  314.98  7332.5  314.27  7461.2  325.25
  7497.4  326.97  7528.1  331.24  7533.7  329.45  7550.5  331.12  7556.1  329.66
  7578.4  328.29  7595.2  329.18  7639.9  328.68  7645.5  327.53  7676.3  327.83
#Mann= 7 ,-1 , 0
  4037.7     .12       0  4375.5     .16       0  4401.6     .05       0
  4402.9    .033       0  4408.9     .05       0  7316.2     .16       0
  7461.2     .12       0
Bank Sta=4363.4,7326.9
XS Rating Curve= 0 ,0
Exp/Cntr=0.3,0.1

Type RM Length L Ch R = 1 ,36418   ,542,542,542
BEGIN DESCRIPTION:
BIG BROWN CREEK 43.0
END DESCRIPTION:
XS GIS Cut Line= 3
      3621199.57     10642760.21      3621999.61     10642360.19
      3624199.64     10640760.17
#Sta/Elev= 30
  4117.4  329.77  4162.2  326.36  4220.9  323.62    4355  315.25  4363.4   311.4
  4377.4   310.6  4408.1  310.95  4435.1  309.78  4452.9  309.89  4458.2  303.61
    4461  303.11  4464.2  303.61  7274.7  303.61  7281.2  309.72  7295.9  309.59
  7310.6  310.99  7324.1  312.51  7331.5  314.85  7352.3  314.86  7390.1  317.87
  7431.9   320.4  7452.8  320.75  7488.2  324.71  7546.7  328.23  7567.9  330.41
  7645.6  334.77  7674.6  333.74  7689.3  334.18  7695.5  333.23  7732.2  332.26
#Mann= 6 ,-1 , 0
  4117.4     .12       0  4435.1     .05       0  4458.2    .033       0
  4464.2     .05       0  7390.1     .16       0  7488.2     .12       0
Bank Sta=4363.4,7331.5
XS Rating Curve= 0 ,0
Exp/Cntr=0.3,0.1

Type RM Length L Ch R = 1 ,35876   ,540,540,540
BEGIN DESCRIPTION:
BIG BROWN CREEK 42.0
END DESCRIPTION:
XS GIS Cut Line= 3
      3621449.59     10644360.22      3622299.61     10642810.19
      3624299.59     10640810.21
#Sta/Elev= 30
  3230.8  358.64  3304.2  357.11  3369.7  352.45  3385.8  346.75  3401.9  350.86
  3429.4  350.06  3766.9  328.39  3777.3  329.49    3783  325.33  3799.1  324.47
  3804.8  328.88  3820.9  324.52  3835.3  326.83  3973.5  319.07  4033.2  315.88
  4092.9  310.77  4158.3  309.91  4171.4  303.61  4174.2  303.11  4177.4  303.61
  7346.2  303.61  7355.9  308.13  7367.4  311.82  7374.5  318.27  7445.2  326.53
  7517.6  330.17  7649.2   337.2  7658.5  337.62    7728  339.74    7827  337.98
#Mann= 9 ,-1 , 0
  3230.8     .05       0  3304.2     .16       0  3973.5     .12       0
  4171.4    .033       0  4177.4     .12       0  7355.9     .16       0
  7517.6     .12       0  7649.2     .08       0  7658.5     .12       0
Bank Sta=4033.2,7374.5
XS Rating Curve= 0 ,0
Exp/Cntr=0.3,0.1

Type RM Length L Ch R = 1 ,35336   ,541,541,541
BEGIN DESCRIPTION:
BIG BROWN CREEK 41.0
END DESCRIPTION:
XS GIS Cut Line= 3
      3621799.59     10644060.21      3622599.61     10643260.19
      3624399.61     10640860.19
#Sta/Elev= 30
  3863.2  332.96  3905.7  330.67  4089.5  316.22  4117.8  315.38  4160.2  311.58
  4226.8  309.75  4230.9  309.68  4242.1  303.61  4244.8  303.11  4248.1  303.61
  7381.1  303.61  7387.3  309.63  7401.9  313.28  7424.6  315.34  7431.1  316.43
  7494.6  321.15  7501.9  322.66  7531.1  325.28  7587.3  328.79  7601.9   332.9
  7632.6  334.28  7674.3  337.01  7687.3  336.28  7716.5  338.84  7781.1  340.33
  7787.3  339.71  7858.1  343.25  7944.6  345.18  7987.3  344.94  7994.6  343.77
#Mann= 7 ,-1 , 0
  3863.2     .16       0  4226.8     .05       0  4242.1    .033       0
  4248.1     .05       0  7424.6     .16       0  7632.6     .08       0
  7674.3     .12       0
Bank Sta=4089.5,7431.1
XS Rating Curve= 0 ,0
Exp/Cntr=0.3,0.1

Type RM Length L Ch R = 1 ,34795   ,563,563,563
BEGIN DESCRIPTION:
BIG BROWN CREEK 40.0
END DESCRIPTION:
XS GIS Cut Line= 3
      3621599.61     10644360.19      3622899.61     10643710.19
      3624899.63     10641710.17
#Sta/Elev= 30
  3541.4  358.67  3577.7   357.8  3586.1  356.24  3639.2  353.07  3661.6  348.65
  3678.6  349.29  3697.9  347.93  3711.9  344.63  3773.4  338.01  3787.4  338.23
  3795.8  335.63  3894.2  328.99    3997  322.14  4002.6  322.71    4092  313.96
  4094.7  312.64  4100.4  309.84  4114.4  310.48  4159.1   309.8  4164.5  303.61
  4167.2  303.11  4170.5  303.61  4234.2  303.61  7271.7  303.61    7300  317.05
  7346.7  320.52  7483.9  327.13  7554.6  333.91  7646.5   339.6  7823.3  337.86
#Mann= 9 ,-1 , 0
  3541.4     .05       0  3678.6     .16       0  3894.2     .12       0
  4094.7     .16       0  4164.5    .033       0  4170.5     .16       0
  4234.2     .05       0  7346.7     .12       0  7646.5     .05       0
Bank Sta=4114.4,7300
XS Rating Curve= 0 ,0
Exp/Cntr=0.3,0.1

Type RM Length L Ch R = 1 ,34232   ,548,548,548
BEGIN DESCRIPTION:
BIG BROWN CREEK 39.0
END DESCRIPTION:
XS GIS Cut Line= 3
      3621649.66     10644510.18      3623249.61     10644160.19
      3625649.63     10642760.18
#Sta/Elev= 30
  3382.6  358.44  3433.7  356.18    3444  350.55  3464.4  347.44  3474.7  351.88
  3499.9  349.86  3525.9  345.18  3536.1  338.37  3543.6  338.95  3548.9  339.15
  3556.6  335.26  3607.8  333.42  3658.5  324.49  3827.5  314.48  3853.4  310.78
  3904.6  309.79  3914.8  308.44  3917.3  303.61  3920.1  303.11  3923.3  303.61
  3952.2  303.61  6849.6  303.61  6861.5  309.51  6890.7  310.28  6994.7  313.09
  7039.8  311.45  7193.8  310.08  7333.8  313.96  7550.4  329.18  7798.9  338.94
#Mann= 10 ,-1 , 0
  3382.6     .05       0  3543.6     .16       0  3658.5     .12       0
  3917.3    .033       0  3923.3     .12       0  3952.2     .05       0
  6890.7     .16       0  7039.8     .08       0  7193.8     .16       0
  7333.8     .12       0
Bank Sta=3827.5,6994.7
XS Rating Curve= 0 ,0
Exp/Cntr=0.3,0.1

Type RM Length L Ch R = 1 ,33684   ,531,531,531
BEGIN DESCRIPTION:
BIG BROWN CREEK 38.0
END DESCRIPTION:
XS GIS Cut Line= 3
      3622099.64     10645860.16      3623549.61     10644610.19
       3625749.6      10642810.2
#Sta/Elev= 30
  3060.5  343.56  3081.9  339.59  3102.7  339.98  3131.2  333.26  3138.9  335.39
  3190.4  329.72  3229.1  325.95  3315.5  319.35  3401.1  319.51  3450.5  316.35
  3456.3  312.76  3464.7  314.65  3484.7  310.89  3514.1  308.07  3613.9  310.44
    3649  314.98  3755.5  317.87  3894.7  315.09  3925.5  314.67  3932.1  310.68
  3936.8  303.61  3939.5  303.11  3942.8  303.61  6993.6  303.61  7000.5  303.61
    7007  309.87  7134.8  318.65  7266.2  322.39  7668.1  338.74  7817.4  338.08
#Mann= 10 ,-1 , 0
  3060.5     .05       0  3190.4     .16       0  3229.1     .12       0
  3456.3     .07       0  3484.7     .12       0  3894.7     .05       0
  3936.8    .033       0  3942.8     .05       0  6993.6     .16       0
  7266.2     .12       0
Bank Sta=3755.5,7134.8
XS Rating Curve= 0 ,0
Exp/Cntr=0.3,0.1

Type RM Length L Ch R = 1 ,33153   ,1004,1004,1004
BEGIN DESCRIPTION:
BIG BROWN CREEK 37.0
END DESCRIPTION:
XS GIS Cut Line= 3
       3622749.6     10645660.19      3623899.61     10645010.19
       3625699.6      10643010.2
#Sta/Elev= 30
  3680.7   328.8  3834.5  321.39  3936.9  314.21  3952.9  312.75  3955.6  303.61
  3958.3  303.11  3961.6  303.61    4012  303.61  6977.5  303.61  6984.2   309.3
  6991.7   309.9  7019.7  310.03    7041  313.06  7047.8  312.44  7055.2   313.8
  7118.8   313.8  7125.3  314.56  7140.4  315.18  7161.4  313.91  7168.1  311.82
  7175.6  316.02  7182.3  314.96  7189.8  316.51  7196.5  315.73  7251.4  317.92
  7281.7  318.49  7310.1   320.7  7444.6  326.43  7628.5  337.21  7692.4  339.08
#Mann= 6 ,-1 , 0
  3680.7     .12       0  3955.6    .033       0  3961.6     .12       0
    4012     .05       0  7125.3     .16       0  7251.4     .12       0
Bank Sta=3936.9,7140.4
XS Rating Curve= 0 ,0
Exp/Cntr=0.3,0.1

Type RM Length L Ch R = 1 ,32149   ,514,514,514
BEGIN DESCRIPTION:
BIG BROWN CREEK 35.0
END DESCRIPTION:
XS GIS Cut Line= 4
      3622181.53     10646065.74      3624264.84     10645926.86
       3624820.4     10645649.08      3626017.51     10643393.65
#Sta/Elev= 30
  2626.3  344.64  2739.3  342.52    2970  331.36  3025.3  328.32  3082.2  322.36
  3115.5  321.46  3155.6   315.7  3175.6  310.66  3205.7  309.62  3305.9  310.02
  3380.4  314.54  3388.7  315.31  3479.8  314.78  3490.1   314.6  3778.1  310.18
    3807  309.59    3817  307.88    3824  303.61  3826.8  303.11    3830  303.61
  6435.1  303.61  6443.6  309.79  6447.8  309.82  6511.5  311.28  6621.6   322.8
  6687.6  326.21  6813.8  326.52  7035.2  320.66  7352.2  321.09  7888.8  336.82
#Mann= 12 ,-1 , 0
  2626.3     .05       0  2739.3     .16       0    2970     .12       0
  3082.2     .16       0  3380.4     .12       0  3479.8     .16       0
  3490.1     .12       0  3778.1     .05       0    3824    .033       0
    3830     .05       0  6447.8     .16       0  7035.2     .12       0
Bank Sta=3388.7,6443.6
XS Rating Curve= 0 ,0
Exp/Cntr=0.3,0.1

Type RM Length L Ch R = 1 ,31635   ,307,307,307
BEGIN DESCRIPTION:
BIG BROWN CREEK 34.0
END DESCRIPTION:
XS GIS Cut Line= 4
      3622371.91     10646837.21      3624559.44     10646355.43
      3625132.35     10646042.93       3626108.9     10643829.43
#Sta/Elev= 30
  2441.3  323.91  2477.7  322.76  2490.1  322.27  2496.2  320.86  2572.1  321.62
  2593.9  321.12  2623.3   318.4  2637.6  318.92  2730.2  317.36  2817.7  313.82
  2822.8  314.67  2889.5  310.92    2910   312.6  2920.5  310.11  2951.7   309.9
  2971.4  310.08  2978.6  303.61  2981.4  303.11  2984.6  303.61  7085.6  303.61
  7094.8  309.81  7162.2  309.92  7170.5  310.84  7216.8  310.65  7390.7   316.6
  7396.4  317.57  7593.9  324.39  7632.1  326.63    7646   328.4  7753.2   333.4
#Mann= 7 ,-1 , 0
  2441.3     .12       0  2477.7     .16       0  2951.7     .05       0
  2978.6    .033       0  2984.6     .05       0  7170.5     .16       0
  7390.7     .12       0
Bank Sta=2910,7094.8
XS Rating Curve= 0 ,0
Exp/Cntr=0.3,0.1

Type RM Length L Ch R = 1 ,31328   ,1324,1324,1324
BEGIN DESCRIPTION:
BIG BROWN CREEK 33.0
END DESCRIPTION:
XS GIS Cut Line= 4
       3623304.2     10649662.77      3624892.77     10646563.77
      3625322.46     10646186.16      3628498.34     10645014.73
#Sta/Elev= 30
  1335.6  341.95  1518.3  342.11  1613.6  337.41  2022.6  321.34  2112.4  319.08
    2278  316.69  2574.6  311.58  2605.3  309.67  2607.9  303.61  2610.7  303.11
  2613.9  303.61  2619.5  309.55  2627.5  309.76  2633.1  303.61  2655.3  303.61
  2660.8  307.57  2716.3   309.7  2721.9  303.61  7507.7  303.61  7518.7  309.54
  7563.4  310.55  7588.5  315.52  7614.7  317.28  7796.2  330.25    7902  328.61
  8109.7  333.48  8312.1  329.75  8428.5  321.39  8453.6  326.33  8775.1   334.2
#Mann= 9 ,-1 , 0
  1335.6     .05       0  1613.6     .16       0  2022.6     .05       0
  2112.4     .16       0  2607.9    .033       0  2613.9     .16       0
  2660.8     .05       0  7507.7     .16       0  7614.7     .12       0
Bank Sta=2278,7588.5
XS Rating Curve= 0 ,0
Exp/Cntr=0.3,0.1

Type RM Length L Ch R = 1 ,30004   ,694,694,694
BEGIN DESCRIPTION:
BIG BROWN CREEK 31.0
END DESCRIPTION:
XS GIS Cut Line= 4
       3624098.5      10649649.7      3625647.98     10647631.47
      3626090.69     10647305.95      3628043.78     10645990.87
#Sta/Elev= 30
  2204.7  334.81  2391.1  327.42  2405.6  324.13  2432.6  326.45  2497.1  324.81
  2540.7   319.3  2611.3  322.74  2640.4  322.46  2661.2   319.3  2675.7  322.09
  2793.8  322.49  2939.4  323.93  2968.5  321.36  3001.4  325.46  3025.5  326.47
  3153.3  330.98  3225.3  330.04  3645.5  309.74  3703.5   309.8  3706.9  303.61
  3709.6  303.11  3712.9  303.61  6447.3  303.61  6454.7  309.93  6601.1  310.34
  6629.5  310.87  6717.8  310.75  6930.1  310.61  7319.9  331.56  7653.2  332.61
#Mann= 10 ,-1 , 0
  2204.7     .16       0  2432.6     .12       0  2793.8     .16       0
  3001.4     .12       0  3025.5     .05       0  3706.9    .033       0
  3712.9     .05       0  6601.1     .12       0  6629.5     .05       0
  6717.8     .12       0
Bank Sta=3703.5,6454.7
XS Rating Curve= 0 ,0
Exp/Cntr=0.3,0.1

Type RM Length L Ch R = 1 ,29310   ,722,722,722
BEGIN DESCRIPTION:
BIG BROWN CREEK 30.0
END DESCRIPTION:
XS GIS Cut Line= 3
      3624849.64     10649260.17      3626299.61     10648010.19
      3627899.61     10646210.19
#Sta/Elev= 30
  3109.1   337.6  3194.1  334.92  3257.7  330.04  3293.9  330.09  3307.1  328.08
  3456.3  320.74    3577  313.11  3626.4  310.82  3640.6  311.29  3704.3  309.25
  3708.9  303.61  3711.7  303.11  3714.9  303.61    6780  303.61  6787.5  307.22
  6794.2   306.9  6796.8  307.87  6801.7  309.69  6914.6  311.03  6922.1  309.62
    6943  310.16  6999.9  314.74  7056.8  317.76  7247.4  323.59  7361.1  328.38
  7367.8  329.91  7389.6  329.62  7396.3  331.71  7403.8  330.47  7431.8  332.02
#Mann= 4 ,-1 , 0
  3109.1     .05       0  3708.9    .033       0  3714.9     .05       0
  6796.8     .12       0
Bank Sta=3640.6,6914.6
XS Rating Curve= 0 ,0
Exp/Cntr=0.3,0.1

Type RM Length L Ch R = 1 ,28588   ,772,772,772
BEGIN DESCRIPTION:
BIG BROWN CREEK 29.0
END DESCRIPTION:
XS GIS Cut Line= 4
       3625205.3     10649558.54      3626650.58     10648699.18
      3626897.98     10648373.66      3628082.85     10646290.37
#Sta/Elev= 30
  3176.2  332.44  3204.5  331.36  3375.8  325.39  3390.6  320.59  3412.8  323.37
  3448.3  321.34  3503.5   318.8  3565.1   316.3  3571.5  312.86  3578.3  314.31
  3588.1  309.83  3593.9   315.1    3600  310.53  3623.3  311.16    3631  313.17
  3643.6  303.61  3646.3  303.11  3649.6  303.61  6914.1  303.61  6919.9  308.59
  6935.7  310.28  6950.1     310  6963.1  313.29  6986.4  315.25  6986.7  315.26
  7205.3  326.92  7301.8  327.82  7388.3  331.08  7536.9  331.24  7663.2  327.49
#Mann= 9 ,-1 , 0
  3176.2     .05       0  3204.5     .16       0  3448.3     .05       0
  3503.5     .16       0  3571.5     .05       0  3643.6    .033       0
  3649.6     .05       0  6986.4     .16       0  6986.7     .12       0
Bank Sta=3631,6935.7
XS Rating Curve= 0 ,0
Exp/Cntr=0.3,0.1

Type RM Length L Ch R = 1 ,27816   ,638,638,638
BEGIN DESCRIPTION:
BIG BROWN CREEK 28.0
END DESCRIPTION:
XS GIS Cut Line= 4
      3624825.75     10650212.06       3626976.1     10649389.29
      3627418.81      10649024.7       3628655.2     10645888.19
#Sta/Elev= 30
  2377.1  348.95  2460.2  346.29  2586.6  339.34  2723.7  332.67  2755.4  323.71
  2790.8   325.1  2798.8  316.95  2820.8  325.43  2875.6  316.94  2900.3  322.78
  3087.9  321.23  3223.1  313.26  3288.2  309.48  3309.7  303.61  3312.5  303.11
  3315.7  303.61  7123.4  303.61  7194.3  303.61  7227.2  305.85  7434.8  317.35
  7477.5  318.44  7493.8  316.73  7538.6  315.98  7856.5  303.61  7861.9  309.52
  7964.8  309.85  8240.9  330.21  8487.2  325.69  8525.5  319.22  8624.4  328.24
#Mann= 14 ,-1 , 0
  2377.1     .08       0  2460.2     .05       0  2586.6     .08       0
  2723.7     .05       0  3223.1     .16       0  3288.2     .05       0
  3309.7    .033       0  3315.7     .05       0  7123.4     .16       0
  7194.3     .05       0  7227.2     .16       0  7434.8     .12       0
  7493.8     .16       0  7538.6     .12       0
Bank Sta=3087.9,7477.5
XS Rating Curve= 0 ,0
Exp/Cntr=0.3,0.1

Type RM Length L Ch R = 1 ,27178   ,505,505,505
BEGIN DESCRIPTION:
BIG BROWN CREEK 26.0
END DESCRIPTION:
XS GIS Cut Line= 3
      3625540.15     10651824.65      3627677.76      10649741.3
      3628749.61     10646610.19
#Sta/Elev= 30
  1787.5  325.95  1822.7  325.33    1840  324.82  2056.2  325.43  2087.3   326.5
  2129.7  319.69    2165  327.75  2249.9  328.04  2306.4  308.62  2310.6  303.61
  2313.4  303.11  2316.6  303.61  2427.7  303.61  2532.8  303.61  2589.4  326.75
  2614.7   326.7  2845.4  325.81  3088.6  326.07  3276.2  320.14  3374.4  311.14
  3395.2  309.85  3423.8  303.61    7696  303.61  7733.1  310.18  7753.3  303.61
  7758.6  309.47  7788.4  312.69  7946.4  322.42  7986.8   329.3  8081.9  331.68
#Mann= 13 ,-1 , 0
  1787.5     .05       0  1822.7      .1       0    1840     .15       0
  2056.2      .1       0  2310.6    .033       0  2316.6      .1       0
  2427.7     .05       0  2614.7     .08       0  2845.4     .16       0
  3088.6     .12       0  3276.2     .16       0  3395.2     .05       0
  7788.4     .12       0
Bank Sta=3374.4,7733.1
XS Rating Curve= 0 ,0
Exp/Cntr=0.3,0.1

Type RM Length L Ch R = 1 ,26673   ,524,524,524
BEGIN DESCRIPTION:
BIG BROWN CREEK 25.0
END DESCRIPTION:
XS GIS Cut Line= 3
      3625999.62     10652160.17      3628199.61     10649760.19
       3628899.6     10646860.22
#Sta/Elev= 30
  1740.2  333.62  1994.7  326.62  2072.8  318.06  2185.9  326.15  2330.7  320.58
  2381.2  303.61    2384  303.11  2387.2  303.61  2433.9  303.61  2674.3  303.61
  2738.2   330.4  2978.6  316.72  3053.8  312.71  3096.3  311.05  3206.7  306.07
  3224.7  305.17  3359.7  322.15  3512.6  325.23  3573.1  328.18    3610  326.07
  3738.4  310.82  3785.8  303.61  6846.2  303.61  6954.7  313.28    7074  319.21
  7325.4  303.61  7536.9  303.61  7748.8  319.19  7855.8   314.1  7979.2  332.09
#Mann= 20 ,-1 , 0
  1740.2     .05       0  1994.7      .1       0  2185.9     .15       0
  2330.7      .1       0  2381.2    .033       0  2387.2      .1       0
  2433.9     .05       0  2674.3     .16       0  2978.6     .12       0
  3053.8     .16       0  3096.3     .05       0  3206.7     .12       0
  3224.7     .05       0  3359.7     .16       0  3512.6     .12       0
    3610     .16       0  3738.4     .05       0  6954.7     .16       0
  7325.4     .05       0  7748.8     .12       0
Bank Sta=3573.1,7074
XS Rating Curve= 0 ,0
Exp/Cntr=0.3,0.1

Type RM Length L Ch R = 1 ,26149   ,580,580,580
BEGIN DESCRIPTION:
BIG BROWN CREEK 24.0
END DESCRIPTION:
XS GIS Cut Line= 3
      3627744.56     10653510.84      3628720.89     10649790.76
      3629059.44     10647277.73
#Sta/Elev= 30
  1365.6  321.82  1560.2  325.08  1958.7  323.73  1986.6  319.02  2462.2  325.15
  2513.9  320.38  2606.9  322.08  2710.3  319.76  2813.7  310.74  2931.5  310.28
    2935  310.34  2982.6   309.6  2986.4  303.61  2989.2  303.11  2992.4  303.61
  3035.3  303.61  6170.8  303.61  6180.9  303.82    6191  309.51  6242.3  310.57
  6438.1  319.03  6620.4  314.85  6718.8  312.21  6817.3  312.07  7014.1  314.35
  7414.3  314.81  7487.1  323.74  7492.7  330.67  7510.3  330.36  7747.4  330.35
#Mann= 12 ,-1 , 0
  1365.6     .05       0  2931.5     .16       0    2935     .12       0
  2986.4    .033       0  2992.4     .12       0  3035.3     .05       0
  6242.3     .16       0  6620.4     .08       0  6718.8     .05       0
  6817.3      .1       0  7014.1     .05       0  7510.3     .12       0
Bank Sta=2606.9,6438.1
XS Rating Curve= 0 ,0
Exp/Cntr=0.3,0.1

Type RM Length L Ch R = 1 ,25569   ,116,116,116
BEGIN DESCRIPTION:
BIG BROWN CREEK 23.0
END DESCRIPTION:
XS GIS Cut Line= 4
      3629654.29     10653536.89      3629212.95     10650281.48
      3628987.82     10648575.48      3629117.95     10647404.37
#Sta/Elev= 30
  1566.6  321.67  1879.4   323.8  1978.9  323.23  2376.8  319.05    2411   319.4
  2612.8  309.49  2619.9  303.61  2622.6  303.11  2625.9  303.61  2895.3  311.58
  2955.9  309.52    2966  303.61  3570.6  303.61    3792  303.61  4167.5  303.61
    4267  303.61  4937.4  303.61  5360.9  303.61  5460.4  303.61  5930.2  303.61
  6104.6  303.61  6245.1  303.61    6272  309.56    6554  320.49  6608.1  322.51
  6848.9  314.93  7143.6   315.2  7553.9  314.62  7656.7  330.61  7750.9  329.43
#Mann= 20 ,-1 , 0
  1566.6     .05       0  1879.4      .1       0  1978.9     .16       0
  2376.8     .05       0  2619.9    .033       0  2625.9     .05       0
  3570.6     .08       0    3792     .05       0  4167.5     .08       0
    4267     .05       0  4937.4     .05       0  5360.9      .1       0
  5460.4     .05       0  5930.2     .05       0  6104.6     .05       0
    6272     .16       0    6554     .05       0  6848.9     .08       0
  7143.6     .05       0  7656.7     .12       0
Bank Sta=2411,6608.1
XS Rating Curve= 0 ,0
Exp/Cntr=0.3,0.1

Type RM Length L Ch R = 1 ,25453   ,409,409,409
BEGIN DESCRIPTION:
Mapping XS f23472d9
END DESCRIPTION:
XS GIS Cut Line= 4
      3629690.95      10653009.1      3629137.56     10648853.26
      3629137.56     10648592.85      3629236.75     10647279.02
#Sta/Elev= 30
  2064.4   323.6  2095.7  323.63  2337.6  322.31  2735.4  322.35  2945.9  322.16
  3016.1  297.16  3018.8  296.66  3022.1  297.16  3102.4  304.86  3133.1  319.36
  3152.8  322.52  3431.4  322.95  3630.3  322.74  3834.7  322.52    4227  321.18
  4525.3  321.61  4724.2   321.4  5022.5   321.6  5320.8   321.9  5619.1  320.77
    5818  319.98  6116.3  318.82  6608.6  323.25  6790.8  314.72  7302.2  314.74
  7342.3  326.22  7372.4  315.41  7482.7  314.27  7636.5  324.05  7834.9  320.06
#Mann= 20 ,-1 , 0
  2064.4     .05       0  2095.7      .1       0  2337.6     .05       0
  2735.4     .05       0  3016.1     .04       0  3022.1      .1       0
  3133.1     .05       0  3431.4      .1       0  3630.3     .05       0
  3834.7      .1       0    4227     .05       0  4525.3      .1       0
  4724.2     .05       0  5022.5      .1       0  5320.8     .05       0
  5619.1      .1       0    5818     .05       0  6116.3     .08       0
  6608.6     .05       0  7636.5     .12       0
Bank Sta=2945.9,3152.8
XS Rating Curve= 0 ,0
Exp/Cntr=0.3,0.1

Type RM Length L Ch R = 1 ,25044   ,967,967,967
BEGIN DESCRIPTION:
BIG BROWN CREEK 22.0
END DESCRIPTION:
XS GIS Cut Line= 6
      3629929.66     10652802.91      3629851.54     10651526.87
      3629708.31      10650042.5      3629669.24     10649860.21
      3629395.81     10648506.04      3629408.81     10647543.85
#Sta/Elev= 30
  2187.8  301.95  2340.4  299.47    2421  286.23  2491.6  286.51  2551.2     278
    2602  284.87  2706.7  279.51    2764  291.64  2811.7  289.99    2918  248.79
  2920.7  248.29    2924  248.79  3082.2  248.82  3172.4  284.15  3254.9  293.99
  3543.3  274.78  4115.7  257.43  4267.3  255.98  5366.4  257.05  5570.7  269.46
    5677  277.22  5914.6  295.74  6015.4  304.12  6194.7  318.79  6715.8  308.95
  7107.9     313  7221.3  311.06  7251.3  298.21  7281.3  311.43  7487.7  313.05
#Mann= 14 ,-1 , 0
  2187.8     .05       0  2340.4     .16       0  2491.6     .12       0
  2706.7     .05       0    2918     .03       0    2924     .05       0
  4115.7     .16       0  4267.3     .05       0  5570.7     .16       0
    5677     .05       0  5914.6     .16       0  6015.4     .12       0
  6715.8     .05       0  7107.9     .12       0
Bank Sta=3254.9,6194.7
XS Rating Curve= 0 ,0
Exp/Cntr=0.3,0.1

Type RM Length L Ch R = 1 ,24077   ,1190,1190,1190
BEGIN DESCRIPTION:
BIG BROWN CREEK 20.0
END DESCRIPTION:
XS GIS Cut Line= 3
      3630546.83     10652321.47      3630582.87     10650366.57
      3630478.81     10648363.31
#Sta/Elev= 30
  2843.8  303.31  3035.8  298.96  3254.9  292.54  3409.4  288.11  3700.7     279
  3975.3   266.5  4132.3  248.79  4135.1  248.29  4138.3  248.79  4156.5  248.79
  4744.5  249.65  4815.4  249.94  4885.5  259.76  4945.6  258.92  4995.7  250.37
  5035.7  260.94  5105.8  263.15  5406.2  262.22  5461.7  253.74    5877  256.41
  6017.1  253.74  6273.5  261.21  6318.5  262.31  6437.6   273.5  6477.7  284.46
  6487.7  296.45  6501.6  297.15  6515.3  310.27  6613.7  325.56    6805  330.63
#Mann= 15 ,-1 , 0
  2843.8     .05       0  3035.8     .12       0  3254.9     .16       0
  3409.4     .12       0  3700.7     .16       0  4132.3     .07       0
  4138.3     .16       0  4156.5     .05       0  4744.5     .16       0
  5461.7     .07       0    5877     .16       0  6273.5     .12       0
  6318.5     .05       0  6515.3     .16       0  6613.7     .12       0
Bank Sta=3975.3,5105.8
XS Rating Curve= 0 ,0
Exp/Cntr=0.3,0.1

Type RM Length L Ch R = 1 ,22887   ,859,859,859
BEGIN DESCRIPTION:
Mapping XS 665d492a
END DESCRIPTION:
XS GIS Cut Line= 4
      3630989.44     10651434.29      3631579.71     10650271.11
      3631597.07      10650010.7      3630746.59      10648604.8
#Sta/Elev= 30
  3501.8   293.9  3934.4  261.92  4002.4  261.25  4041.3  254.56  4247.3  253.08
  4328.8  253.05  4549.3  252.51  4957.4  255.95  4981.2  251.76  5004.5  249.07
  5007.3  248.57  5010.5  249.07  5047.6  254.91  5091.6  254.22  5115.4  254.51
  5866.2  256.54    6169  269.12  6289.1  277.76  6348.6  281.96  6558.7  298.58
  6577.5  293.84  6601.4  285.56  6616.9  301.04  6622.8  294.88  6632.4     300
  6641.3   293.4  6653.8  304.25  6659.6  299.91  6675.1  308.09  6710.3  312.28
#Mann= 15 ,-1 , 0
  3501.8     .05       0  3934.4     .12       0  4247.3     .07       0
  4328.8     .12       0  4549.3     .05       0  4981.2     .16       0
  5004.5     .07       0  5010.5     .16       0  5091.6     .16       0
  5115.4     .05       0    6169     .16       0  6289.1     .12       0
  6348.6     .16       0  6577.5     .05       0  6641.3     .16       0
Bank Sta=4957.4,5047.6
XS Rating Curve= 0 ,0
Exp/Cntr=0.3,0.1

Type RM Length L Ch R = 1 ,22028   ,240,240,240
BEGIN DESCRIPTION:
BIG BROWN CREEK 19.0
END DESCRIPTION:
XS GIS Cut Line= 3
      3631107.03     10651558.04      3631701.24     10650600.97
      3632621.27     10648734.88
#Sta/Elev= 30
    4124  297.85  4285.2   287.6  4327.7  276.73  4333.6  283.59  4437.6  283.08
  4536.5  276.03  4589.9  261.85  4726.9   263.1  4730.9  262.21  4765.7  258.38
  4865.5   254.5    4922  248.72  5153.8  247.71  5156.5  247.21  5159.8  247.71
  5285.6  255.09  5622.4  252.59  6127.5  253.83  6526.3  253.86  6584.2  262.56
  6588.1  263.06  6891.7  272.15    6981  275.28  6997.9   281.1  7048.3  277.97
  7132.6  284.67  7138.2  279.88  7177.5  285.28  7183.1  280.74  7331.1  288.89
#Mann= 11 ,-1 , 0
    4124     .05       0  4730.9     .16       0  4765.7     .05       0
  4865.5     .16       0    4922     .05       0  5153.8     .03       0
  5159.8     .05       0  5622.4     .07       0  6127.5     .05       0
  6584.2     .07       0  6891.7     .05       0
Bank Sta=4726.9,6588.1
XS Rating Curve= 0 ,0
Exp/Cntr=0.3,0.1

Type RM Length L Ch R = 1 ,21788   ,1056,1056,1056
BEGIN DESCRIPTION:
BIG BROWN CREEK 18.0
END DESCRIPTION:
XS GIS Cut Line= 2
      3631348.82     10651664.75      3632867.06     10648953.61
#Sta/Elev= 30
  4141.4  302.26  4174.5  304.01  4190.5  300.71  4196.2  303.95  4271.5  298.55
  4277.2  302.65  4314.9  297.89  4320.6  302.12  4336.6  298.75  4439.3  297.54
    4461  300.81  4725.9  269.84  4850.3  260.71  4893.7  258.51  4960.4  248.11
  5166.7  250.28  5177.2   246.5    5180     246  5183.2   246.5  5212.1  253.02
  5277.2   256.3  5546.6  254.16  5940.9   253.2  6401.7  253.79  6423.3   258.1
  6702.5  256.19  6731.6  261.72  6759.8  269.38  6862.9  278.48  7248.7  297.75
#Mann= 5 ,-1 , 0
  4141.4     .05       0  5177.2     .03       0  5183.2     .05       0
  5546.6     .07       0  5940.9     .05       0
Bank Sta=4850.3,6731.6
XS Rating Curve= 0 ,0
Exp/Cntr=0.3,0.1

Type RM Length L Ch R = 1 ,20732   ,1738,1738,1738
BEGIN DESCRIPTION:
BIG BROWN CREEK 17.0
END DESCRIPTION:
XS GIS Cut Line= 3
      3632794.99      10651807.6      3632786.31       10650410.
        3633081.     10649153.22
#Sta/Elev= 30
  4162.9  286.22  4230.3  286.15  4290.3  283.07  4490.3  267.28  4580.3  261.57
  4630.3  260.03  4680.3  255.13  4720.3  253.11  4870.3  250.76  4960.3  253.61
  4970.3  252.78  4980.3  246.53  4987.3  244.43  4990.1  243.93  4993.3  244.43
  5000.3  245.87  5020.3  253.74  5180.3  251.38  5700.9  252.18  5846.7  252.42
  5981.5  250.87  6340.9  251.59  6476.3   257.7  6603.6  267.23  6638.8  268.51
  6651.2  270.74  6688.5  272.15  6778.5  282.91  6839.1  287.51  6851.4  288.48
#Mann= 7 ,-1 , 0
  4162.9     .05       0  4987.3     .03       0  4993.3     .05       0
  5700.9     .16       0  5846.7     .05       0  6340.9     .12       0
  6839.1     .16       0
Bank Sta=4960.3,5020.3
XS Rating Curve= 0 ,0
Exp/Cntr=0.3,0.1

Type RM Length L Ch R = 1 ,18994   ,1024,1024,1024
BEGIN DESCRIPTION:
Mapping XS a09cf07c
END DESCRIPTION:
XS GIS Cut Line= 2
      3633654.36     10651998.56      3633758.53      10648890.9
#Sta/Elev= 30
  3548.1  281.45  3776.6  273.49  4036.7  261.24  4220.7  255.37  4597.1   248.5
  4913.6  250.45  4967.3  251.43  4977.3   251.1  4987.3  244.64  4994.3  242.76
    4997  242.26  5000.3  242.76  5004.6  244.85  5017.3  250.86  5102.6  250.92
  5192.9  249.71  5477.6  248.93  5897.8  259.38  5907.8  258.36  5937.8  260.37
  5967.8  255.07  5984.4  255.82  6027.9  256.05  6037.9  259.52  6067.9  264.34
  6147.9  269.05  6429.4  278.65  6478.1  279.43  6618.3  287.16  6657.5  290.46
#Mann= 11 ,-1 , 0
  3548.1     .16       0  4220.7     .05       0  4913.6     .16       0
  4994.3     .07       0  5000.3     .16       0  5004.6     .12       0
  5102.6     .16       0  5192.9     .05       0  5984.4     .16       0
  6429.4     .12       0  6618.3     .16       0
Bank Sta=4967.3,5017.3
XS Rating Curve= 0 ,0
Exp/Cntr=0.3,0.1

Type RM Length L Ch R = 1 ,17970   ,1761,1761,1761
BEGIN DESCRIPTION:
Mapping XS f4e84c38
END DESCRIPTION:
XS GIS Cut Line= 3
       3633616.6     10652489.43      3634538.91     10650395.24
      3634213.39     10648865.28
#Sta/Elev= 30
  2837.1  298.39  2964.9   295.5  3034.5  296.55  3203.3  290.93  3255.4  293.27
  3437.3  294.78    3773   270.5  3808.8  266.36  3923.7  258.97  4033.4  253.99
  4061.6  252.88  4158.4   248.5  4373.4  246.53  4453.5  247.14  4469.7  245.31
  4481.9   247.1  4910.8  249.48  4969.2  249.98  4993.4  246.46  4996.8  241.43
  4999.5  240.93  5002.8  241.43  5015.8  241.73  5039.2  249.67  5253.2  247.15
  5508.8  247.27  5958.3  253.74  6295.1   266.6  6551.7  282.18  6689.6   285.3
#Mann= 11 ,-1 , 0
  2837.1     .12       0  2964.9     .16       0    3773     .05       0
  4033.4     .08       0  4061.6     .05       0  4373.4     .16       0
  4481.9     .05       0  4910.8     .16       0  4993.4     .05       0
  4996.8     .03       0  5002.8     .05       0
Bank Sta=4969.2,5039.2
XS Rating Curve= 0 ,0
Exp/Cntr=0.3,0.1

Type RM Length L Ch R = 1 ,16209   ,239,239,239
BEGIN DESCRIPTION:
BIG BROWN CREEK 16.0
END DESCRIPTION:
XS GIS Cut Line= 6
      3634094.01     10653422.62      3634430.41     10652934.31
      3634484.66     10652532.83      3634593.17     10652304.97
      3635363.56     10651111.39      3634614.85      10648745.9
#Sta/Elev= 30
  2806.4   298.6    2964  285.59  3199.6  268.72  3294.8   266.5  3437.7  263.48
  3918.3  259.42  4552.2  245.53    4979  247.59  4992.6  240.05    5003  239.99
  5005.8  239.49    5009  239.99  5015.3  241.21  5021.2  247.71  5039.4   247.7
  5153.2   245.5    5161  245.48  5267.1  246.51  6868.9  248.07  7261.7  258.04
  7305.5  262.63  7331.6  259.21  7401.4  259.28  7588.7  266.48  7627.6  271.54
  7659.9  266.58  7714.6  266.75    7762  271.66  7914.6  273.79  7960.3  274.79
#Mann= 11 ,-1 , 0
  2806.4     .12       0    2964     .05       0  3294.8     .07       0
  3437.7     .05       0    5003     .04       0    5009     .05       0
  5039.4     .16       0  5153.2     .05       0    5161     .08       0
  5267.1     .05       0  7914.6     .16       0
Bank Sta=4979,5021.2
XS Rating Curve= 0 ,0
Exp/Cntr=0.3,0.1

Type RM Length L Ch R = 1 ,15970   ,1918,1918,1918
BEGIN DESCRIPTION:
BIG BROWN CREEK 15.0
END DESCRIPTION:
XS GIS Cut Line= 6
      3634245.95     10653563.64      3634647.42     10653021.11
      3634723.37     10652641.34      3634766.78     10652456.88
      3635537.18      10651263.3      3634755.91     10648778.45
#Sta/Elev= 30
  2765.5  287.99  2863.6  283.58  3134.9  262.73    3363  255.37  3553.5  257.38
  4203.7  247.76  4465.5  248.08  4509.1  239.25    4537  244.88  4573.1  245.22
  4597.3  245.33  4941.6  247.42  4971.7  246.99  4986.9  239.46  4998.1  239.23
  5000.9  238.73  5004.1  239.23    5008  246.63    5014  244.13  5052.7  247.33
  5516.4  244.89  5543.5  248.48  5570.8  247.05  5581.2  249.12  5710.2  246.61
  7055.4  249.61  7390.9  262.35  7464.2   262.3  7846.9  278.37  8042.6  280.78
#Mann= 9 ,-1 , 0
  2765.5     .12       0    3363     .05       0  4573.1     .12       0
  4597.3     .16       0  4998.1     .07       0  5004.1     .16       0
  5052.7     .05       0  5570.8     .08       0  5710.2     .05       0
Bank Sta=4941.6,5052.7
XS Rating Curve= 0 ,0
Exp/Cntr=0.3,0.1

Type RM Length L Ch R = 1 ,14052   ,834,834,834
BEGIN DESCRIPTION:
BIG BROWN CREEK 14.0
END DESCRIPTION:
XS GIS Cut Line= 3
       3634242.5     10653828.88      3636011.03      10652208.5
      3634745.97     10648518.96
#Sta/Elev= 30
  2767.6  304.13  3111.5  272.23  3383.9  256.01  3649.2  246.78  3854.6  245.55
  3868.8  248.45  3939.7  244.36  4080.9  242.18  4802.3  244.43  4897.2  244.24
  4965.8  245.49  4973.2  245.27  4992.4  237.06  4998.5  235.88  5001.3  235.38
  5004.5  235.88  5008.3  240.35  5022.5  245.16  5135.9  243.09  5990.2  245.15
  6110.9  244.85  6434.1   246.4  6539.2   246.5  7064.4  249.63  7470.9  247.97
  7715.8  249.59    8362   268.1  8557.9  278.52    8758  285.29  9066.6  284.89
#Mann= 11 ,-1 , 0
  2767.6     .12       0  3383.9     .05       0  4802.3     .16       0
  4897.2     .12       0  4992.4     .05       0  4998.5     .03       0
  5004.5     .05       0  5990.2     .12       0  6110.9     .05       0
  6434.1     .08       0  6539.2     .05       0
Bank Sta=4965.8,5022.5
XS Rating Curve= 0 ,0
Exp/Cntr=0.3,0.1

Type RM Length L Ch R = 1 ,13218   ,1200,1200,1200
BEGIN DESCRIPTION:
BIG BROWN CREEK 13.0
END DESCRIPTION:
XS GIS Cut Line= 3
      3634520.27     10654262.91      3636673.06     10652578.87
      3639196.77     10647629.04
#Sta/Elev= 30
  3067.5  311.25  3360.5  280.37  3695.5  258.51  4116.4  242.23  4670.8  241.29
  4963.7  244.96  4989.7  234.89  4992.4  234.39  4995.7  234.89  5021.6  243.87
  5477.3  238.81  5624.4  246.32  5804.5  254.14  6375.2  246.42  6411.2  246.89
  6921.5  258.33  7550.5  258.04  8021.9  256.21  8129.9  254.84  9748.7  272.94
  9856.6   276.3 10151.8  285.88 10537.4  311.61 10612.1   317.2 10647.2  319.54
   10720  324.34 10842.9  332.97 11074.9  357.89 11216.2  362.57 11356.8  357.41
#Mann= 20 ,-1 , 0
  3067.5     .12       0  3695.5     .05       0  4670.8     .12       0
  4989.7     .07       0  4995.7     .12       0  5624.4     .05       0
  6375.2     .12       0  6411.2     .05       0  7550.5     .12       0
  8021.9     .16       0  8129.9     .05       0  9748.7     .16       0
  9856.6     .12       0 10151.8     .16       0 10537.4     .05       0
 10612.1     .12       0 10647.2     .16       0   10720     .12       0
 10842.9     .16       0 11216.2     .16       0
Bank Sta=4963.7,5021.6
XS Rating Curve= 0 ,0
Exp/Cntr=0.3,0.1

Type RM Length L Ch R = 1 ,12018   ,1885,1885,1885
BEGIN DESCRIPTION:
BIG BROWN CREEK 12.0
END DESCRIPTION:
XS GIS Cut Line= 3
      3634927.71      10654711.1       3637057.9     10653132.98
      3639847.26     10649307.01
#Sta/Elev= 30
  3069.5  282.92  3072.8  282.92  3300.3  270.15  3677.1  250.47  3697.7  249.33
  3936.5  239.84  4422.8  239.74    4980  243.51  4994.6  237.59  4997.9  233.63
  5000.6  233.13  5003.9  233.63  5015.4  236.01  5023.8  242.05    5030  242.11
  5385.3  241.92  5576.5  242.26  6009.2  255.43  6431.8  252.79  6912.1  259.34
  7219.9  254.69  7551.6  255.23  7875.7  257.42  8110.6  256.93  9473.8     267
 10067.8  275.56 10100.8  278.84 10174.7  278.94 10331.8  286.68 10455.4  291.19
#Mann= 16 ,-1 , 0
  3069.5     .12       0  3072.8     .05       0  3300.3     .12       0
  3677.1     .07       0  3697.7     .12       0  4997.9     .07       0
  5003.9     .12       0  5385.3     .07       0  5576.5     .05       0
  7219.9     .12       0  7551.6     .05       0  7875.7     .12       0
  8110.6     .05       0 10100.8     .16       0 10174.7     .12       0
 10331.8     .16       0
Bank Sta=4980,5030
XS Rating Curve= 0 ,0
Exp/Cntr=0.3,0.1
