--- CANEY CREEK.prj (project) ---

Proj Title=CANEY CREEK Base Level Engineering
Current Plan=p01
Default Exp/Contr=0.3,0.1
English Units
Geom File=g01
Flow File=f01
Plan File=p01
Y Axis Title=Elevation
X Axis Title(PF)=Main Channel Distance
X Axis Title(XS)=Station
BEGIN DESCRIPTION:
CANEY CREEK
END DESCRIPTION:
DSS File=dss
DSS Export Rating Curves= 0
DSS Export Rating Curve Sorted= 0
DSS Export Volume Flow Curves= 0
DXF OffsetX= 0
DXF OffsetY= 0
DXF ScaleX= 1
DXF ScaleY= 10

--- CANEY CREEK.p01 (plan) ---

Plan Title=Multiple Run
Program Version=4.10
Short Identifier=Multiple Run
Geom File=g01
Flow File=f01
Subcritical Flow
K Sum by GR= 0
Std Step Tol= 0.01
Critical Tol= 0.01
Num of Std Step Trials= 20
Max Error Tol= 0.3
Flow Tol Ratio= 0.001
Split Flow NTrial= 30
Split Flow Tol= 0.02
Split Flow Ratio= 0.02
Log Output Level= 0
Friction Slope Method= 1
Unsteady Friction Slope Method= 2
Unsteady Bridges Friction Slope Method= 1
Parabolic Critical Depth
Global Vel Dist= 1 , 1 , 1
Global Log Level= 0
CheckData=True
Encroach Param=-1 ,0,0, 0
BEGIN DESCRIPTION:
Multiple Run
END DESCRIPTION:
Computation Interval=1HOUR
Output Interval=1HOUR
Run HTab= 0
Run UNet= 0
Run PostProcess= 0
Run WQNet= 0
UNET Theta= 1
UNET Theta Warmup= 1
UNET ZTol= 0.02
UNET ZSATol= 0.05
UNET MxIter= 20
UNET MaxInSteps= 0
UNET DtIC= 0
UNET DtMin= 0
UNET MaxCRTS= 20
UNET WFStab= 2
UNET SFStab= 1
UNET WFX= 1
UNET SFX= 1
UNET DSS MLevel= 4
UNET DZMax Abort= 100
UNET Convert EG Bridges= 0
UNET Use Existing IB Tables=-1
UNET Froude Reduction=False
UNET Froude Limit= 1
UNET Froude Power= 10
UNET Time Slicing=0,0, 5
UNET Junction Losses=0
Instantaneous Interval=1HOUR
DSS File=dss
Write IC File= 0
Write IC File at Sim End=0
Echo Input=False
Echo Parameters=False
Echo Output=False
Write Detailed= 0
WQ AD Non Conservative
WQ ULTIMATE=-1
WQ Max Comp Step=1HOUR
WQ Output Interval=15MIN
WQ Output Selected Increments= 0
WQ Output face flow=0
WQ Output face velocity=0
WQ Output face area=0
WQ Output face dispersion=0
WQ Output cell volume=0
WQ Output cell surface area=0
WQ Output cell continuity=0
WQ Output cumulative cell continuity=0
WQ Output face conc=0
WQ Output face dconc_dx=0
WQ Output face courant=0
WQ Output face peclet=0
WQ Output face adv mass=0
WQ Output face disp mass=0
WQ Output cell mass=0
WQ Output cell source sink temp=0
WQ Output cell source sink nsm=0
WQ Output MaxMinRange=-1
WQ Daily Max Min Mean=-1
WQ Daily Range=0
WQ Daily Time=0
WQ Create Restart=0
WQ Fixed Restart=0
WQ System Summary=0
WQ Use Fixed Temperature=0
Sorting and Armoring Iterations= 10
XS Update Threshold= 0.02
Hydraulics Update Threshold= 0.02
Energy Slope Method= 1
Volume Change Method= 0
XS Weighting Method= 0
Number of US Weighted Cross Sections= 1
Number of DS Weighted Cross Sections= 1
Upstream XS Weight=0.25
Main XS Weight=0.5
Downstream XS Weight=0.25
Number of DS XS's Weighted with US Boundary= 1
Upstream Boundary Weight= 1
Weight of XSs Associated with US Boundary= 0
Number of US XS's Weighted with DS Boundary= 1
Downstream Boundary Weight= 0.5
Weight of XSs Associated with DS Boundary= 0.5
Sediment Output Level= 4
Mass or Volume Output= 0
Output Increment Type= 1
Profile and TS Output Increment= 10
XS Output Flag= 0
XS Output Increment= 10
Disregard all LS=0
Disregard all Conn=0
Disregard all Breaches=0
Disregard all Pumps=0

--- CANEY CREEK.f01 (steady flow) ---

Flow Title=Multiple
Program Version=4.10
Number of Profiles= 7
Profile Names=10-year,25-year,50-year,1pct_min,100-year,1pct_plu,500-year
River Rch & RM=CANEY CREEK,Reach-1         ,116284
    2493    3543    4438    4051    5478    7408    8322
River Rch & RM=CANEY CREEK,Reach-1         ,112892
    2762    3936    4938    4512    6102    8252    9291
River Rch & RM=CANEY CREEK,Reach-1         ,108529
    4476    6507    8275    7649   10345   13990   16129
River Rch & RM=CANEY CREEK,Reach-1         ,102728
    5781    8484   10858   10092   13649   18458   21518
River Rch & RM=CANEY CREEK,Reach-1         ,101774
    5781    8484   10858   10092   13649   18458   21518
River Rch & RM=CANEY CREEK,Reach-1         ,99860
    5904    8640   11036   10234   13841   18718   21721
River Rch & RM=CANEY CREEK,Reach-1         ,94876
    7776   11499   14792   13806   18671   25250   29678
River Rch & RM=CANEY CREEK,Reach-1         ,92856
    7776   11499   14792   13806   18671   25250   29678
River Rch & RM=CANEY CREEK,Reach-1         ,91782
    7776   11499   14792   13806   18671   25250   29678
River Rch & RM=CANEY CREEK,Reach-1         ,84602
    8088   11878   15206   14116   19090   25816   30012
River Rch & RM=CANEY CREEK,Reach-1         ,79274
    8156   11930   15229   14116   19090   25816   30012
River Rch & RM=CANEY CREEK,Reach-1         ,75416
    8156   11930   15229   14116   19090   25816   30012
River Rch & RM=CANEY CREEK,Reach-1         ,68201
   14875   22124   28576   26725   36142   48878   57637
River Rch & RM=CANEY CREEK,Reach-1         ,66803
   14875   22124   28576   26725   36142   48878   57637
River Rch & RM=CANEY CREEK,Reach-1         ,65962
   14875   22124   28576   26725   36142   48878   57637
River Rch & RM=CANEY CREEK,Reach-1         ,65245
   14875   22124   28576   26725   36142   48878   57637
River Rch & RM=CANEY CREEK,Reach-1         ,62790
   14875   22124   28576   26725   36142   48878   57637
River Rch & RM=CANEY CREEK,Reach-1         ,60942
   14875   22124   28576   26725   36142   48878   57637
River Rch & RM=CANEY CREEK,Reach-1         ,57109
   14875   22124   28576   26725   36142   48878   57637
River Rch & RM=CANEY CREEK,Reach-1         ,56128
   14875   22124   28576   26725   36142   48878   57637
River Rch & RM=CANEY CREEK,Reach-1         ,46983
   14897   22124   28576   26725   36142   48878   57637
River Rch & RM=CANEY CREEK,Reach-1         ,44193
   15523   23009   29648   27655   37400   50579   59319
River Rch & RM=CANEY CREEK,Reach-1         ,43624
   15523   23009   29648   27655   37400   50579   59319
River Rch & RM=CANEY CREEK,Reach-1         ,40034
   15523   23009   29648   27655   37400   50579   59319
River Rch & RM=CANEY CREEK,Reach-1         ,39304
   18229   27076   34944   32634   44133   59685   70155
River Rch & RM=CANEY CREEK,Reach-1         ,35803
   18229   27076   34944   32634   44133   59685   70155
River Rch & RM=CANEY CREEK,Reach-1         ,31807
   19336   28784   37205   34799   47062   63645   75034
River Rch & RM=CANEY CREEK,Reach-1         ,29672
   19336   28784   37205   34799   47062   63645   75034
River Rch & RM=CANEY CREEK,Reach-1         ,28372
   19375   28807   37205   34799   47062   63645   75034
River Rch & RM=CANEY CREEK,Reach-1         ,22646
   19910   29599   38225   35716   48301   65322   76846
River Rch & RM=CANEY CREEK,Reach-1         ,20295
   19910   29599   38225   35716   48301   65322   76846
River Rch & RM=CANEY CREEK,Reach-1         ,16006
   19910   29599   38225   35716   48301   65322   76846
River Rch & RM=CANEY CREEK,Reach-1         ,14454
   19910   29599   38225   35716   48301   65322   76846
Boundary for River Rch & Prof#=CANEY CREEK,Reach-1         , 1
Up Type= 0
Dn Type= 3
Dn Slope=0.0013
Boundary for River Rch & Prof#=CANEY CREEK,Reach-1         , 2
Up Type= 0
Dn Type= 3
Dn Slope=0.0013
Boundary for River Rch & Prof#=CANEY CREEK,Reach-1         , 3
Up Type= 0
Dn Type= 3
Dn Slope=0.0013
Boundary for River Rch & Prof#=CANEY CREEK,Reach-1         , 4
Up Type= 0
Dn Type= 3
Dn Slope=0.0013
Boundary for River Rch & Prof#=CANEY CREEK,Reach-1         , 5
Up Type= 0
Dn Type= 3
Dn Slope=0.0013
Boundary for River Rch & Prof#=CANEY CREEK,Reach-1         , 6
Up Type= 0
Dn Type= 3
Dn Slope=0.0013
Boundary for River Rch & Prof#=CANEY CREEK,Reach-1         , 7
Up Type= 0
Dn Type= 3
Dn Slope=0.0013
DSS Import GetInterval= 0
DSS Import GetPeak= 0
DSS Import FillOption= 0

--- CANEY CREEK.g01 (geometry) ---

Geom Title=Existing Conditions
Program Version=4.10

River Reach=CANEY CREEK     ,Reach-1
Reach XY= 30
       3566169.5       10584930.       3566749.5       10586373.
      3566114.25       10588723.      3564343.25       10590222.
        3564034.       10594603.      3561764.25       10596327.
      3561300.75       10598140.      3562939.75       10602616.
        3561403.       10604261.       3561191.5       10606395.
        3562387.       10607641.      3562208.75       10609496.
      3563682.25       10609324.      3564546.75       10611421.
      3563434.75       10612048.      3563241.75       10614095.
        3566347.       10617504.      3564358.75       10623610.
       3565107.5       10623881.       3564867.5       10625677.
      3566416.25       10626646.      3565379.25       10628362.
       3566489.5       10631114.      3563691.75       10639862.
      3564024.25       10644093.      3561772.25       10647731.
       3563186.5       10652079.        3560955.       10656929.
      3563582.25       10658160.       3564559.5       10661181.

Type RM Length L Ch R = 1 ,116284  ,416,416,416
BEGIN DESCRIPTION:
CANEY CREEK 159.0
END DESCRIPTION:
XS GIS Cut Line= 3
      3565849.58      10585260.2      3566199.61     10585160.19
      3566549.57     10584910.22
#Sta/Elev= 30
    4639  455.72  4649.4  455.36  4655.9  454.49  4694.9   452.9  4701.4  452.04
    4795  446.58  4801.5  445.54  4815.8  444.97  4826.2  443.64  4867.8  441.36
  4874.3  440.01  4879.5  440.04    4899   438.1  4930.2  437.98  4952.3  438.98
  4971.8  438.45  4986.1  436.74  5007.4  435.72  5010.2  435.22  5013.4  435.72
  5016.5  436.42  5052.2  438.81  5125.9  439.19  5182.5  438.69  5253.7  440.37
    5298  443.37    5325  446.58  5375.4  450.33  5404.9  453.14  5433.1  452.37
#Mann= 3 ,-1 , 0
    4639     .05       0  5007.4     .03       0  5013.4     .05       0
Bank Sta=4952.3,5052.2
XS Rating Curve= 0 ,0
Exp/Cntr=0.3,0.1

Type RM Length L Ch R = 1 ,115868  ,110,110,110
BEGIN DESCRIPTION:
CANEY CREEK 158.0
END DESCRIPTION:
XS GIS Cut Line= 3
      3566149.61     10585760.19      3566549.61     10585360.19
      3566749.61     10585010.19
#Sta/Elev= 30
  4469.8  456.55  4597.1  452.53  4710.2  444.46  4879.9  443.26  4936.5  441.84
  4978.9  439.21  5004.2  432.41    5007  431.91  5010.2  432.41  5021.3  439.27
  5035.5  439.84    5065  439.69  5070.8  441.31  5080.8   440.4  5086.6  441.67
  5102.4  440.76  5108.2  442.13    5124  440.36  5129.8  441.57  5161.5  440.85
  5167.2  442.07  5204.7  441.37  5210.4  442.68  5242.1  443.15  5247.8  444.59
  5277.4  446.88  5300.4  451.45  5350.1   452.1  5371.7  455.22  5438.6  457.97
#Mann= 3 ,-1 , 0
  4469.8     .05       0  5004.2     .03       0  5010.2     .05       0
Bank Sta=4978.9,5035.5
XS Rating Curve= 0 ,0
Exp/Cntr=0.3,0.1

Type RM Length L Ch R = 1 ,115758  ,692,692,692
BEGIN DESCRIPTION:
CANEY CREEK 157.0
END DESCRIPTION:
XS GIS Cut Line= 4
      3566194.92     10585812.32      3566490.07     10585590.09
      3566667.15     10585388.71      3566854.56     10585045.12
#Sta/Elev= 30
  4460.7   455.4  4529.2  453.33  4558.1  447.71  4601.8  444.01  4651.8  443.78
    4658  445.45  4672.6  445.99  4687.2  444.83  4693.4  446.21  4722.6  445.73
  4751.7  442.73  4826.7  439.25  4886.2  437.73  4893.8  438.71  4971.6  439.07
  4978.2  436.77  4985.8  432.17  5011.3  432.15    5014  431.65  5017.3  432.15
  5020.9  435.49  5028.5  436.69  5070.3  436.61    5165  439.35  5255.3  443.99
  5260.9  446.27  5282.8   447.8  5298.9  447.62  5313.1  449.43  5489.7  458.72
#Mann= 3 ,-1 , 0
  4460.7     .05       0  5011.3     .03       0  5017.3     .05       0
Bank Sta=4978.2,5028.5
XS Rating Curve= 0 ,0
Exp/Cntr=0.3,0.1

Type RM Length L Ch R = 1 ,115066  ,465,465,465
BEGIN DESCRIPTION:
Mapping XS 13f7efdb
END DESCRIPTION:
XS GIS Cut Line= 3
      3566195.45     10586045.85      3566877.73     10586103.14
      3567615.98     10585863.99
#Sta/Elev= 30
  4435.3  454.25  4476.9  452.82  4569.9  448.85    4600  445.79  4620.1  442.07
  4670.9  437.88  4760.6  437.63  4770.6  438.85  4810.8   434.9  4941.2  433.18
  5008.5  430.62  5011.2  430.12  5014.5  430.62  5020.7  432.13  5081.7  432.68
    5147  431.77  5195.5  433.64    5307  435.07  5408.2  438.19  5434.9  437.66
  5458.3  440.14  5498.9   438.8  5594.9  441.59  5600.2  443.07    5616  443.85
  5701.4  445.87  5721.1   445.1  5795.7  447.13  5862.7  447.66    5896   448.4
#Mann= 6 ,-1 , 0
  4435.3     .08       0  4476.9     .05       0  5008.5     .03       0
  5014.5     .05       0  5795.7     .08       0  5862.7     .05       0
Bank Sta=4941.2,5081.7
XS Rating Curve= 0 ,0
Exp/Cntr=0.3,0.1

Type RM Length L Ch R = 1 ,114601  ,133,133,133
BEGIN DESCRIPTION:
CANEY CREEK 156.0
END DESCRIPTION:
XS GIS Cut Line= 2
      3566066.96     10586085.77      3567146.12     10586891.89
#Sta/Elev= 30
    4266  456.44  4296.2  455.89  4348.6   454.7  4364.1  452.43  4384.9  453.41
  4449.6  450.39  4464.2  451.59    4485  449.64  4493.4  450.78  4499.6  448.14
  4506.5  449.49  4543.4  448.68  4594.1  445.17  4749.7  437.87  4778.9  434.78
  4799.8  435.81  4862.6  432.94  4935.3  431.95  4993.3     424  5003.1  423.92
  5005.9  423.42  5009.1  423.92  5020.7  428.14  5035.3  427.35  5043.2   429.4
  5085.3  431.36  5229.2  433.89  5279.2  441.27  5435.5  450.26    5613  451.71
#Mann= 6 ,-1 , 0
    4266     .05       0  4296.2     .08       0  4594.1     .05       0
  4862.6     .08       0  5003.1     .07       0  5009.1     .08       0
Bank Sta=4935.3,5085.3
XS Rating Curve= 0 ,0
Exp/Cntr=0.3,0.1

Type RM Length L Ch R = 1 ,114468  ,331,331,331
BEGIN DESCRIPTION:
CANEY CREEK 155.0
END DESCRIPTION:
XS GIS Cut Line= 2
       3565962.8     10586168.24      3567078.27     10587010.27
#Sta/Elev= 30
  4223.4  457.68  4293.1  456.88  4386.4  456.79  4480.1  453.77  4500.9   455.3
  4515.5  452.82  4629.9  446.41  4736.1  437.31  4781.9  435.61  4799.1  434.67
  4944.2  432.52  4971.3  429.49  4979.6  424.43  4985.9   425.2  4997.5  419.29
  5000.2  418.79  5003.5  419.29  5033.9  427.28  5044.1  430.34  5058.7  431.93
  5094.1  431.82  5100.4  430.15  5185.7  431.47    5194  433.49  5214.8  432.82
  5229.4  437.29  5258.5  439.87  5340.3  444.99  5449.4  449.68    5621   451.6
#Mann= 9 ,-1 , 0
  4223.4     .08       0  4293.1     .05       0  4781.9     .08       0
  4799.1     .05       0  4997.5     .03       0  5003.5     .05       0
  5033.9     .08       0  5340.3     .05       0  5449.4     .08       0
Bank Sta=4944.2,5058.7
XS Rating Curve= 0 ,0
Exp/Cntr=0.3,0.1

Type RM Length L Ch R = 1 ,114137  ,230,230,230
BEGIN DESCRIPTION:
CANEY CREEK 154.0
END DESCRIPTION:
XS GIS Cut Line= 3
      3566099.62      10586560.2      3566399.61     10586910.19
      3566599.63      10587010.2
#Sta/Elev= 30
  4525.2  456.58  4532.3  456.19  4538.9  453.02  4546.6  451.67  4581.7  449.79
  4638.8  444.89  4667.3  443.58  4688.2  441.24  4723.3  439.44  4745.3  437.69
  4766.1  434.61  4794.6  434.43  4829.8   432.1    4866  430.83  4915.4  430.23
  4972.4  431.21    4979  430.69  4982.9  428.88    4989  428.88  4994.6  420.22
  4997.1  420.05  4999.9  419.55  5003.1  420.05  5008.5  423.57  5016.9  430.53
  5067.2  430.57  5075.6  429.88  5111.9  429.51  5156.7  431.69  5209.8   435.9
#Mann= 3 ,-1 , 0
  4525.2     .05       0  4997.1     .03       0  5003.1     .05       0
Bank Sta=4972.4,5016.9
XS Rating Curve= 0 ,0
Exp/Cntr=0.3,0.1

Type RM Length L Ch R = 1 ,113907  ,594,594,594
BEGIN DESCRIPTION:
CANEY CREEK 153.0
END DESCRIPTION:
XS GIS Cut Line= 2
      3565651.28     10586567.98      3566743.87     10587495.81
#Sta/Elev= 30
  4173.7  453.06  4230.9   453.6  4237.4  452.28  4507.7  443.11  4564.8  439.41
  4571.4  437.61  4606.5  436.97  4649.3  433.42  4692.2  434.84  4727.3  431.61
    4791  429.79  4961.3  430.14    4969   429.4  4983.3  422.79  5001.1  418.95
  5003.9  418.45  5007.1  418.95  5011.1  426.52    5025  429.74  5145.8  428.55
  5217.2  431.22  5260.1     432  5266.6   430.9  5295.2  433.76    5316   432.8
  5344.6  434.47  5373.2  438.74  5457.7  438.25    5494  441.96  5607.1  447.61
#Mann= 3 ,-1 , 0
  4173.7     .05       0  5001.1     .03       0  5007.1     .05       0
Bank Sta=4961.3,5025
XS Rating Curve= 0 ,0
Exp/Cntr=0.3,0.1

Type RM Length L Ch R = 1 ,113313  ,421,421,421
BEGIN DESCRIPTION:
CANEY CREEK 152.0
END DESCRIPTION:
XS GIS Cut Line= 3
      3565273.53     10586982.66      3565999.61     10587260.19
      3566399.61     10587660.19
#Sta/Elev= 30
    4200  456.76  4281.4  455.81    4319  452.91    4335  453.14  4373.8   450.3
  4403.8  449.85  4409.9  448.55    4464  446.36  4483.3  444.27  4628.3  437.71
  4707.8  431.98  4792.6  430.91  4822.7  428.87  4852.7   428.2  4955.9   427.2
  4967.6  426.51  4974.6  418.74  4980.8  418.74  4988.4   414.8  4991.2   414.3
  4994.4   414.8  5005.6     415  5019.7  426.94  5062.2  428.58  5274.3  428.13
  5288.4  429.84  5359.1  434.39  5401.6  436.27  5436.9  439.55    5543  445.38
#Mann= 3 ,-1 , 0
    4200     .05       0  4988.4     .03       0  4994.4     .05       0
Bank Sta=4955.9,5062.2
XS Rating Curve= 0 ,0
Exp/Cntr=0.3,0.1

Type RM Length L Ch R = 1 ,112892  ,616,616,616
BEGIN DESCRIPTION:
CANEY CREEK 151.0
END DESCRIPTION:
XS GIS Cut Line= 2
      3565304.09      10587258.1      3566445.12     10587726.66
#Sta/Elev= 30
  4181.9  459.95  4220.3  459.79  4226.3  458.42  4317.6  454.03  4327.6  451.74
  4425.7  444.82  4487.6  439.11  4695.6  425.54  4831.7   427.6  4967.8  426.48
  4986.4  416.22  4991.8  415.81  4995.6  414.07  4998.4  413.57  5001.6  414.07
  5009.5  415.24  5015.8  423.89  5021.2   422.1  5039.7  426.85  5052.7  427.54
  5085.1  430.36    5117  431.43  5160.8  435.43  5214.9  438.11  5229.2   440.2
  5277.1  442.18  5282.5  443.53  5330.5  444.59  5354.4  446.72  5415.4  446.82
#Mann= 3 ,-1 , 0
  4181.9     .05       0  4995.6     .03       0  5001.6     .05       0
Bank Sta=4967.8,5052.7
XS Rating Curve= 0 ,0
Exp/Cntr=0.3,0.1

Type RM Length L Ch R = 1 ,112276  ,985,985,985
BEGIN DESCRIPTION:
CANEY CREEK 150.0
END DESCRIPTION:
XS GIS Cut Line= 3
      3565381.65     10587836.81      3565742.75     10587947.92
      3566430.21     10587892.37
#Sta/Elev= 30
  4527.4  450.18  4586.3  442.45  4624.3  439.33  4629.9   438.1  4682.2  434.12
  4689.7   432.8  4807.8  426.12  4863.6  424.47  4891.1  424.66  4972.3  424.22
  4992.3  418.33  4999.4     411  5002.1   410.5  5012.4   411.3  5022.4  421.66
  5042.5  425.26  5052.5  425.44  5060.4  424.43  5092.7  424.11  5142.8  424.66
  5283.3  430.95    5315   433.1  5333.5   435.4  5373.6  436.78  5393.6  438.36
  5403.7  440.03  5463.9  441.77    5514  442.15  5534.1  443.33  5594.9  443.52
#Mann= 4 ,-1 , 0
  4527.4     .12       0  4891.1     .16       0  4972.3     .16       0
  5052.5     .12       0
Bank Sta=4972.3,5052.5
XS Rating Curve= 0 ,0
Exp/Cntr=0.3,0.1

Type RM Length L Ch R = 1 ,111291  ,587,587,587
BEGIN DESCRIPTION:
CANEY CREEK 149.0
END DESCRIPTION:
XS GIS Cut Line= 3
       3565270.5     10587954.83      3565881.64      10588663.2
      3566366.13     10588587.06
#Sta/Elev= 30
  3845.6  455.68  3891.8  451.03  3933.5  448.98  3947.7  446.34  4004.8   443.2
  4011.4  441.73  4039.9   439.2  4076.1  437.98  4117.8  434.11  4224.2  427.03
  4344.9  422.17  4363.1  422.18  4416.1  422.52  4474.7  421.27  4508.3  420.13
  4631.3  420.43  4678.3  419.35  4896.3  421.75  4971.4  421.14  4981.6  414.64
  5001.6     409  5021.5  414.87  5026.6  415.55  5032.2  420.67  5042.3  425.01
  5053.6  427.13  5062.5  429.49  5089.1  433.01  5143.5   437.6  5271.6  444.17
#Mann= 7 ,-1 , 0
  3845.6     .05       0  4363.1     .12       0  4474.7     .16       0
  4631.3     .16       0  4971.4     .12       0  5032.2     .16       0
  5053.6     .05       0
Bank Sta=4971.4,5032.2
XS Rating Curve= 0 ,0
Exp/Cntr=0.3,0.1

Type RM Length L Ch R = 1 ,110704  ,1042,1042,1042
BEGIN DESCRIPTION:
CANEY CREEK 148.0
END DESCRIPTION:
XS GIS Cut Line= 3
       3564949.6     10588060.18      3565749.61     10588860.19
      3566149.61     10589660.18
#Sta/Elev= 30
    3882  473.05  4009.3  464.72  4150.7  445.86  4207.3  440.84  4235.6  441.23
  4263.8  436.67  4331.6  432.59  4428.9  426.02  4603.3  419.74  4843.1  418.62
  4956.8  419.47    4971  418.77  4985.1  408.29    4999  406.54  5002.2  407.04
  5009.8  413.88  5021.8  413.09  5027.4  417.57  5058.1  420.14  5155.9  418.76
  5460.6  419.03  5491.3  413.66  5496.9  417.97  5505.3  416.86  5513.7  413.01
  5519.3  417.99  5536.1  415.06    5550  418.33  5608.7  421.99  5907.8  437.11
#Mann= 10 ,-1 , 0
    3882     .05       0  4331.6     .12       0  4428.9     .16       0
  4603.3     .16       0  4843.1     .16       0  4956.8     .12       0
  5058.1     .16       0  5155.9     .12       0  5460.6     .12       0
  5608.7     .05       0
#XS Ineff= 1 ,-1
 5463.07 5592.33  419.02
Permanent Ineff=
       F
Bank Sta=4956.8,5058.1
XS Rating Curve= 0 ,0
Exp/Cntr=0.3,0.1

Type RM Length L Ch R = 1 ,109662  ,669,669,669
BEGIN DESCRIPTION:
CANEY CREEK 146.0
END DESCRIPTION:
XS GIS Cut Line= 2
      3565041.36     10588642.37       3565638.6     10589718.79
#Sta/Elev= 30
  4221.3  435.42  4285.8  434.76  4313.2  430.97  4321.7  431.02  4329.2  433.11
  4410.5   430.5    4463  426.35  4519.2  422.08  4535.2  423.37  4540.9  421.78
    4557  423.68  4596.5  423.54  4607.6     423  4643.9  416.92    4660  416.28
  4974.7  417.06  4977.2  416.22  4990.7  411.35  4996.5  405.34  5006.7  407.38
  5012.2  404.74  5015.4  405.24  5019.3  409.02  5028.4  411.77  5034.2  411.46
  5042.2  416.14  5055.9  416.58  5110.9  418.36  5264.4  426.17  5452.3  433.61
#Mann= 7 ,-1 , 0
  4221.3     .05       0    4463      .1       0  4596.5     .12       0
  4977.2     .16       0  5055.9     .12       0  5110.9     .16       0
  5264.4     .05       0
#XS Ineff= 2 , 0
         4604.09  425.73
Permanent Ineff=
       F       F
Bank Sta=4974.7,5055.9
XS Rating Curve= 0 ,0
Exp/Cntr=0.3,0.1

Type RM Length L Ch R = 1 ,108993  ,464,464,464
BEGIN DESCRIPTION:
CANEY CREEK 145.0
END DESCRIPTION:
XS GIS Cut Line= 3
      3564849.62     10589010.22      3565099.61     10589810.19
      3565149.62     10590060.22
#Sta/Elev= 30
  4156.2  429.52  4198.1     427  4237.4  423.47  4275.1  422.97  4292.4  420.86
    4340  418.55  4450.6  415.75  4491.4  416.44  4540.1  415.64  4577.9  414.79
  4810.4  415.06  4877.2  414.05  4907.9  414.38  4940.4  413.23  4952.4  414.95
  4962.9  412.95  4978.1  408.56  4983.8  408.88  4991.7  406.31  4996.9  406.31
  5001.5  403.16  5004.3  402.66  5007.5  403.16  5014.7  410.93  5024.9  415.58
  5075.9   416.7  5137.1   419.8  5177.9  422.83  5194.7  423.16  5249.3   426.8
#Mann= 7 ,-1 , 0
  4156.2     .05       0  4450.6     .16       0  4540.1     .16       0
  4877.2     .16       0  4952.4     .12       0  5024.9     .16       0
  5194.7     .05       0
Bank Sta=4952.4,5024.9
XS Rating Curve= 0 ,0
Exp/Cntr=0.3,0.1

Type RM Length L Ch R = 1 ,108529  ,399,399,399
BEGIN DESCRIPTION:
CANEY CREEK 144.0
END DESCRIPTION:
XS GIS Cut Line= 3
      3564083.13     10589786.57      3564595.25     10589821.29
       3565020.6     10590233.62
#Sta/Elev= 30
    4353   429.9  4620.1  427.26  4650.2   425.4  4669.7  422.25  4710.3  417.84
  4740.4   415.4    4759  414.78  4790.5     413  4830.6  412.51  4850.6  414.04
  4925.2  413.38  4953.5  412.05  4960.5  405.05  4967.7  404.99  4981.6  400.67
  4984.8  401.17  4988.8  403.34    4996   402.4  5002.9  405.43  5010.1  403.47
  5017.1  412.22  5024.3  410.39  5031.2  413.59  5038.4  411.29  5045.4  414.23
  5137.2  414.62  5221.1  419.27  5271.7  421.43  5370.8  427.87  5458.7  431.61
#Mann= 6 ,-1 , 0
    4353     .05       0  4669.7     .16       0    4759     .16       0
  4850.6     .12       0  5045.4     .16       0  5221.1     .05       0
Bank Sta=4850.6,5045.4
XS Rating Curve= 0 ,0
Exp/Cntr=0.3,0.1

Type RM Length L Ch R = 1 ,108130  ,390,390,390
BEGIN DESCRIPTION:
CANEY CREEK 143.0
END DESCRIPTION:
XS GIS Cut Line= 2
      3564048.36     10589986.21      3565029.29     10590342.13
#Sta/Elev= 30
  4583.6  432.45  4649.6  431.37  4702.6  430.36  4712.6  429.37  4765.8  428.73
  4861.5  424.42  4925.3  418.13  4936.9  415.57  4956.8  414.03  4962.2  412.38
  4967.9  411.62  4978.5  408.37  4987.5  404.75  4992.8  401.28  4999.6  399.33
  5010.4  400.85  5018.1  404.03  5023.4  404.07  5031.7  413.47  5042.4  413.95
  5095.5  411.92  5163.2  411.96  5201.9  413.33  5261.3  416.82  5288.3  418.89
  5361.5  422.44  5374.8  423.86  5392.2  424.61  5553.2  432.82  5627.1  435.18
#Mann= 7 ,-1 , 0
  4583.6      .1       0  4649.6     .16       0  4956.8     .12       0
  5042.4     .16       0  5163.2     .12       0  5261.3     .12       0
  5392.2     .05       0
Bank Sta=4956.8,5042.4
XS Rating Curve= 0 ,0
Exp/Cntr=0.3,0.1

Type RM Length L Ch R = 1 ,107740  ,502,502,502
BEGIN DESCRIPTION:
CANEY CREEK 142.0
END DESCRIPTION:
XS GIS Cut Line= 3
      3563987.63     10590216.28      3564195.94     10590454.97
      3565042.32     10590593.86
#Sta/Elev= 30
  4587.6   430.9  4762.6  428.68  4797.2  430.03  4882.7  426.43  4928.4  422.87
  4965.7  414.95  4970.8  414.39  4979.1  410.79  4999.3     400  5006.5  399.39
  5009.2  398.89  5012.5  399.39  5019.6  404.56    5027   408.3  5030.9  409.08
  5039.9  412.46    5050   412.8  5083.3  411.99  5120.9  410.97  5210.3  410.72
  5277.1   412.2  5313.5  414.97  5333.4  414.14    5354  414.67  5455.3  420.34
  5495.2  421.69  5583.5   425.3  5607.3  427.56  5678.3   431.4  5762.1  434.45
#Mann= 8 ,-1 , 0
  4587.6     .05       0  4762.6     .16       0  5006.5     .07       0
  5012.5     .16       0  5030.9     .12       0  5083.3     .07       0
  5210.3     .12       0  5495.2     .05       0
Bank Sta=4965.7,5050
XS Rating Curve= 0 ,0
Exp/Cntr=0.3,0.1

Type RM Length L Ch R = 1 ,107238  ,783,783,783
BEGIN DESCRIPTION:
CANEY CREEK 141.0
END DESCRIPTION:
XS GIS Cut Line= 2
      3563744.58     10591049.58      3564959.83     10590862.95
#Sta/Elev= 30
    4409  432.42  4545.6  434.31  4586.1  432.58  4633.6  429.31  4656.9   429.4
  4677.1  426.77  4701.9  425.97  4765.2  420.43  4788.4  419.57    4851  415.17
  4940.2  411.32  4965.2  410.92  4970.5  411.64  4980.7  411.17  4990.8  401.75
  5000.6  398.08    5011  400.21  5021.1  407.05  5028.5  410.06  5061.6  411.53
  5120.7  410.77  5213.3  409.42  5243.7  410.08    5355  417.07  5395.5  420.22
  5405.6  421.93  5428.5  421.85  5555.1  428.87  5587.7  429.53  5638.5  428.05
#Mann= 5 ,-1 , 0
    4409     .16       0    4851     .12       0  4970.5     .07       0
  5061.6     .12       0  5120.7     .07       0
Bank Sta=4970.5,5061.6
XS Rating Curve= 0 ,0
Exp/Cntr=0.3,0.1

Type RM Length L Ch R = 1 ,106455  ,790,790,790
BEGIN DESCRIPTION:
CANEY CREEK 140.0
END DESCRIPTION:
XS GIS Cut Line= 2
      3563825.67     10591371.85      3565190.34     10591449.98
#Sta/Elev= 30
  4544.4  431.47  4639.3  431.38  4708.6  429.19  4793.3  423.59  4838.8   419.9
    4929  415.85  4948.4  413.24    4969  412.59    4979  409.96  4989.1  405.04
  4996.1  398.55  4998.8  398.05  5019.1  402.89  5029.1     410  5049.2  408.76
  5079.2  410.79  5139.3  410.99  5149.3  410.18  5189.4  411.55  5298.6  410.96
  5319.6  408.97  5349.7  410.22  5369.7  409.03  5419.8  409.09  5439.8   407.8
  5519.9  412.23  5529.9  413.61    5567  414.34  5690.2   419.6  5911.3   426.1
#Mann= 6 ,-1 , 0
  4544.4     .05       0  4639.3     .16       0  4793.3     .12       0
    4979     .07       0  5029.1     .12       0    5567     .16       0
Bank Sta=4979,5029.1
XS Rating Curve= 0 ,0
Exp/Cntr=0.3,0.1

Type RM Length L Ch R = 1 ,105665  ,1046,1046,1046
BEGIN DESCRIPTION:
CANEY CREEK 138.0
END DESCRIPTION:
XS GIS Cut Line= 3
      3563830.94     10591726.03      3564398.62     10591981.23
      3565241.51     10592085.29
#Sta/Elev= 30
  4275.3  427.42  4339.6  423.78  4387.3  418.85  4472.5  410.97  4518.8  408.44
  4541.6  408.35  4611.5  407.47  4686.4  409.58  4959.2  409.12  4969.2     408
  4979.3  404.87  4989.4  404.16  4999.5  397.39  5007.8  396.63  5011.1  397.13
  5019.6  405.93  5029.7  408.62  5039.8  417.58  5049.8  420.01  5094.2  420.66
  5209.1  425.84  5321.9  429.63  5342.6  432.05  5436.1  433.59    5463  433.66
  5499.8  436.02  5506.6  434.94  5580.9  435.93  5684.6  439.13    5747  444.72
#Mann= 8 ,-1 , 0
  4275.3     .05       0  4387.3     .16       0  4541.6     .12       0
  4959.2     .07       0  5029.7     .12       0  5209.1      .1       0
  5436.1     .07       0  5506.6     .12       0
Bank Sta=4959.2,5029.7
XS Rating Curve= 0 ,0
Exp/Cntr=0.3,0.1

Type RM Length L Ch R = 1 ,104619  ,1169,1169,1169
BEGIN DESCRIPTION:
CANEY CREEK 137.0
END DESCRIPTION:
XS GIS Cut Line= 3
      3563256.13     10592524.92      3564176.25     10592498.88
      3565243.96     10592186.37
#Sta/Elev= 30
  4310.5  432.55  4724.1   406.9  4874.2  403.79  4941.8  406.52  4954.2  406.84
  4964.2  405.23  4974.2  400.92  5000.6  396.44  5003.3  395.94  5006.6  396.44
  5024.3  405.78  5032.4  406.87  5034.3  407.13  5547.1  406.73  5693.7  413.77
  5762.8  416.53  5818.5  418.56  5911.8  421.08  5918.7  417.33  5952.2  413.22
  5957.4  416.59  5990.8  413.17    5996  415.54  6024.2  414.81  6029.5  419.27
  6057.6  419.64  6078.5  426.18  6134.7  428.36  6201.8  427.23  6343.5  438.59
#Mann= 9 ,-1 , 0
  4310.5     .05       0  4941.8     .16       0  5000.6     .07       0
  5006.6     .16       0  5032.4     .05       0  5693.7     .08       0
  5762.8     .05       0  5818.5     .16       0  6134.7     .12       0
Bank Sta=4954.2,5034.3
XS Rating Curve= 0 ,0
Exp/Cntr=0.3,0.1

Type RM Length L Ch R = 1 ,103450  ,76,76,76
BEGIN DESCRIPTION:
Mapping XS c9b6cc2f
END DESCRIPTION:
XS GIS Cut Line= 4
      3563501.13     10592901.59      3563782.35     10593349.47
      3563949.02     10593309.54      3565218.64     10592364.26
#Sta/Elev= 30
  4415.7  423.52  4478.8  420.97  4551.9  421.93  4673.8   419.9  4768.3  413.38
  4776.9  409.36  4782.8  409.44  4798.1  404.83  4813.4  404.25  4855.8  405.78
    4960  405.32  4982.9  403.62  4993.1  397.15  5004.2  396.34  5006.9  395.84
  5010.2  396.34  5013.7  400.22    5024  404.55  5044.1  405.94  5208.6  402.78
  5308.7  404.21  5594.4  402.58  5844.6  405.58  6015.6  403.74  6265.9   404.3
  6406.2  409.11  6533.2  415.31  6561.2  416.54  6660.3  422.84  6698.8  425.67
#Mann= 7 ,-1 , 0
  4415.7     .05       0  5004.2    .035       0  5010.2     .05       0
  6406.2     .12       0  6533.2     .07       0  6561.2     .12       0
  6660.3     .07       0
Bank Sta=4960,5044.1
XS Rating Curve= 0 ,0
Exp/Cntr=0.3,0.1

Type RM Length L Ch R = 1 ,103374  ,339,339,339
BEGIN DESCRIPTION:
Mapping XS 33e430dd
END DESCRIPTION:
XS GIS Cut Line= 4
      3563494.61     10592921.54      3563801.88     10593407.19
       3563933.4     10593390.27      3565299.71     10592418.91
#Sta/Elev= 30
  4344.9  424.69  4608.1  418.81  4674.6  413.15  4717.5  403.99  4796.3  405.84
  4863.3  404.84  4884.5  406.65  4899.5  404.44  4967.7  402.58  4987.9  393.46
    5005  392.79  5007.8  392.29    5011  392.79  5018.4  399.25  5028.2  402.79
  5063.5  404.65  5099.1  405.66  5128.6  403.57    5200  404.65  5329.7  402.41
  5659.9  402.91  5859.2  405.27  5967.8  402.86  6274.8  404.11  6440.9   407.3
  6510.9  411.86  6585.7  416.74  6671.3  422.89  6710.5  424.94  6728.6  426.39
#Mann= 7 ,-1 , 0
  4344.9     .05       0    5005     .03       0    5011     .05       0
  6510.9     .07       0  6585.7     .12       0  6671.3     .07       0
  6710.5     .16       0
Bank Sta=4899.5,5063.5
XS Rating Curve= 0 ,0
Exp/Cntr=0.3,0.1

Type RM Length L Ch R = 1 ,103035  ,307,307,307
BEGIN DESCRIPTION:
CANEY CREEK 136.0
END DESCRIPTION:
XS GIS Cut Line= 4
      3563473.13     10592924.22      3563811.67     10593618.67
      3564167.57     10593714.15      3565582.53       10592386.
#Sta/Elev= 30
  4097.3  426.11  4257.3  423.79  4443.1  411.06  4493.7  403.73  4533.3   406.8
  4548.9  406.66  4555.8  403.25  4561.4  406.62  4578.3  402.99  4682.4   405.4
  4781.1  402.02  4935.2  402.99  4950.6  403.48  4999.3  391.19  5002.1  390.69
  5005.3  391.19    5023  401.62  5049.2  403.94    5209   401.4  5256.6  398.78
  5270.8  401.56  5347.9  401.01  5949.7  401.69  6242.8  402.17  6614.9  405.38
  6869.9  417.51  6961.8  425.15  7008.5  427.89  7134.6  440.49    7179  446.16
#Mann= 11 ,-1 , 0
  4097.3     .05       0  4935.2     .16       0  4999.3     .07       0
  5005.3     .16       0    5209     .05       0  5347.9     .16       0
  5949.7      .1       0  6242.8     .05       0  6961.8     .12       0
  7008.5     .05       0  7134.6     .16       0
Bank Sta=4950.6,5049.2
XS Rating Curve= 0 ,0
Exp/Cntr=0.3,0.1

Type RM Length L Ch R = 1 ,102728  ,954,954,954
BEGIN DESCRIPTION:
CANEY CREEK 135.0
END DESCRIPTION:
XS GIS Cut Line= 3
      3563377.65     10593028.41      3563794.31       10593827.
      3565313.41     10594703.74
#Sta/Elev= 30
  4012.7   427.4    4118  423.57  4251.6  410.93  4386.9   402.8  4520.8  403.25
  4780.2  400.75  4970.7   402.6  4977.3  399.23  4986.5  398.51  4992.2  391.41
  4997.4  389.52  5000.1  389.02  5003.4  389.52  5023.5  401.27  5029.6  402.63
  5088.4  400.78  5145.1  401.19  5153.1  401.19    5162  393.79  5174.6  400.71
  5200.9  401.96    5265  400.54  5439.1  401.15  5855.3  398.64  6024.6  401.87
  6042.3  402.56  6230.1  409.57  6260.4  412.11  6476.8  422.49  6667.4  429.79
#Mann= 9 ,-1 , 0
  4012.7     .05       0  4997.4     .03       0  5003.4     .05       0
  5145.1     .16       0  5200.9     .05       0  6024.6     .07       0
  6042.3     .05       0  6260.4     .12       0  6476.8     .16       0
Bank Sta=4970.7,5029.6
XS Rating Curve= 0 ,0
Exp/Cntr=0.3,0.1

Type RM Length L Ch R = 1 ,101774  ,1071,1071,1071
BEGIN DESCRIPTION:
Mapping XS 6f22017e
END DESCRIPTION:
XS GIS Cut Line= 3
      3562561.65     10593453.72      3564089.45      10594721.1
      3565070.35     10594790.54
#Sta/Elev= 30
  3129.7  431.13  3309.9  414.59  3352.8     409  3451.9  402.53  3700.5  400.31
  4062.6  400.77    4099  399.41  4368.6  398.28  4695.3  398.53  4834.2  399.14
  4958.5  400.12  4965.8   399.8  4990.7  386.38  4993.4  385.88  4996.7  386.38
  5000.2   386.8    5008  396.43  5014.5  399.26  5028.8  400.18  5103.1   398.8
  5230.8  397.16  5329.7  397.33  5439.6  399.12  5475.8  399.53  5599.3     406
  5646.2  411.43  5776.6  420.12  5998.8   422.4  6021.9  423.38  6098.1  426.76
#Mann= 12 ,-1 , 0
  3129.7     .05       0  4695.3     .07       0  4834.2     .12       0
  4965.8     .07       0  4990.7     .07       0  4996.7     .07       0
  5103.1     .12       0  5230.8     .07       0  5329.7     .05       0
  5439.6     .16       0  5998.8     .12       0  6021.9     .16       0
Bank Sta=4958.5,5028.8
XS Rating Curve= 0 ,0
Exp/Cntr=0.3,0.1

Type RM Length L Ch R = 1 ,100703  ,843,843,843
BEGIN DESCRIPTION:
CANEY CREEK 134.0
END DESCRIPTION:
XS GIS Cut Line= 3
      3562373.71     10593570.13      3563306.03     10595044.12
      3564945.65     10594955.64
#Sta/Elev= 30
    3514  425.22  3620.6  416.25  3663.8  410.55  3684.8  409.87  3757.8  403.18
  3851.8  398.88    4547  395.94  4808.1  395.78  4865.7  394.48  4969.2  398.59
  4975.1  398.84  4996.3  386.73  5004.7  385.95    5008  386.45  5011.6  392.56
  5017.5  393.47  5026.8  398.49  5199.8  395.77  5371.8  396.84    5452  395.54
  5642.2  396.33  5791.2  395.13  6072.9  396.96  6333.2  398.61  6420.8  401.29
  6493.5  403.66  6543.5  403.26  6763.9  412.76  6858.7   414.4  6900.1  415.24
#Mann= 8 ,-1 , 0
    3514     .16       0  3663.8     .05       0    4547     .12       0
  4969.2      .1       0  5026.8     .12       0  6072.9     .05       0
  6420.8     .16       0  6858.7     .12       0
Bank Sta=4975.1,5026.8
XS Rating Curve= 0 ,0
Exp/Cntr=0.3,0.1

Type RM Length L Ch R = 1 ,99860   ,422,422,422
BEGIN DESCRIPTION:
CANEY CREEK 133.0
END DESCRIPTION:
XS GIS Cut Line= 3
      3561384.12     10593663.89      3563332.07       10595341.
      3563862.73     10595715.58
#Sta/Elev= 30
  2358.2  439.42  2572.4  419.89  2642.6  415.59  2728.2  413.54  3004.7  400.33
  3146.2     399  3281.2  396.29  3791.4   392.8  3834.2  394.19  4217.1  394.07
  4706.4  396.85  4855.6  394.95  4962.4  397.75  4969.5  392.84  4975.7  395.07
  4984.3  384.63  4998.8  383.23  5002.1  383.73  5005.2  387.57  5011.4  387.08
  5026.1  389.85  5040.9  395.62    5048  395.42  5084.8  395.17    5148  398.86
  5213.3  400.71  5385.7  413.48  5427.5  416.79  5500.9  417.93  5578.2  423.35
#Mann= 7 ,-1 , 0
  2358.2     .05       0  3146.2      .1       0  4706.4     .12       0
  4962.4      .1       0  5040.9     .12       0    5148     .16       0
  5385.7     .16       0
Bank Sta=4962.4,5048
XS Rating Curve= 0 ,0
Exp/Cntr=0.3,0.1

Type RM Length L Ch R = 1 ,99438   ,453,453,453
BEGIN DESCRIPTION:
CANEY CREEK 132.0
END DESCRIPTION:
XS GIS Cut Line= 2
      3561291.41      10594134.8      3563659.44     10596113.95
#Sta/Elev= 30
  2509.4  438.68    2668  428.31    2789  415.44  2930.8  405.23  3029.7  401.24
  3321.2  400.25  3420.2  397.97  3584.1  394.14  3966.7  393.03  3988.8  391.07
  4087.7  393.52  4385.8  394.55  4627.8  392.68    4961  395.81  4983.1  391.85
  4989.6  384.92  4996.1  383.54  5018.2  387.09  5024.7  394.26  5032.5  396.01
  5067.7  395.47  5118.2   398.5  5160.1  403.62  5180.9  403.87    5203  407.28
  5223.8  407.07  5309.1  415.38  5458.1  423.92    5560   432.1  5595.6  435.28
#Mann= 7 ,-1 , 0
  2509.4     .05       0  3420.2     .08       0    4961     .07       0
  5032.5     .12       0  5118.2     .16       0  5309.1     .16       0
    5560     .12       0
Bank Sta=4961,5032.5
XS Rating Curve= 0 ,0
Exp/Cntr=0.3,0.1

Type RM Length L Ch R = 1 ,98985   ,216,216,216
BEGIN DESCRIPTION:
CANEY CREEK 131.0
END DESCRIPTION:
XS GIS Cut Line= 3
      3561249.63      10594960.2      3563049.61     10596010.19
      3563349.65     10596260.22
#Sta/Elev= 30
  2932.5  429.28  3106.5  419.74  3116.5  416.91  3187.2  413.92  3218.2  409.76
  3332.1  404.96  3418.1  399.96    3685   393.3  3875.6  391.02    4079  391.22
  4101.8  389.64  4110.4  391.32  4313.9  390.02  4351.1  391.56  4642.4  391.71
  4892.2  393.57  4965.5  395.16  4971.3  394.95  4993.2  384.71  4999.7  383.44
  5002.4  382.94  5005.7  383.44  5008.5  384.53  5013.4  390.45  5019.6  390.45
  5037.8  395.63  5037.9  395.64  5115.9  403.74  5257.8  414.71  5406.9  431.08
#Mann= 8 ,-1 , 0
  2932.5     .05       0  3332.1     .16       0  3418.1     .05       0
  4642.4     .12       0  4892.2     .07       0  4999.7     .07       0
  5005.7     .07       0  5037.9     .16       0
Bank Sta=4965.5,5037.8
XS Rating Curve= 0 ,0
Exp/Cntr=0.3,0.1

Type RM Length L Ch R = 1 ,98769   ,1237,1237,1237
BEGIN DESCRIPTION:
CANEY CREEK 130.0
END DESCRIPTION:
XS GIS Cut Line= 2
      3561173.36     10595537.57      3563345.76     10596328.79
#Sta/Elev= 30
  3142.7  442.83  3500.6   407.1  3516.1  405.42  3521.8  401.91  3532.5  400.74
    3592  399.82  3736.1  390.49  4018.2  389.07  4107.2  390.03  4126.2  386.65
  4139.1   389.6  4203.7   389.8  4496.6  390.82  4947.2  394.21  4950.3   394.5
  4990.5  386.44  4997.9  382.78  5000.6  382.28  5003.9  382.78  5011.8  386.95
  5022.5  387.67  5036.8  394.34  5039.9  394.24  5067.3  394.24  5153.7  400.91
  5209.6   408.9  5288.5  414.61    5296  417.22    5363  424.51  5454.7  431.04
#Mann= 10 ,-1 , 0
  3142.7     .05       0    3592     .16       0  3736.1     .05       0
  4018.2     .16       0  4203.7     .05       0  4496.6     .12       0
  4947.2     .07       0  4997.9     .07       0  5003.9     .07       0
  5039.9     .16       0
Bank Sta=4950.3,5036.8
XS Rating Curve= 0 ,0
Exp/Cntr=0.3,0.1

Type RM Length L Ch R = 1 ,97532   ,71,71,71
BEGIN DESCRIPTION:
CANEY CREEK 128.0
END DESCRIPTION:
XS GIS Cut Line= 6
        3560685.     10596141.43      3561195.44     10596258.62
      3561708.46     10596284.66      3562289.19     10596422.68
      3563153.77     10596420.08      3563658.98     10596477.37
#Sta/Elev= 30
  3878.3   414.9  4288.5  401.85  4883.2  392.41  4933.9  391.35  4994.1   378.5
  4996.9     378  5000.1   378.5  5060.3  392.59    5081   384.9  5086.2  392.05
    5120  380.98  5125.2  390.25  5153.8  383.99    5159  390.73  5236.5  385.24
  5246.7  391.12  5473.1  392.59  5547.8  386.86  5552.8  391.97  5570.9  391.74
  5657.9  382.32  5671.8  387.67  5734.6  384.18  5751.5  392.09  5787.3  393.04
  5886.7  392.76  6283.2  401.83  6382.1  410.25  6691.3  436.84  6895.5  439.75
#Mann= 9 ,-1 , 0
  3878.3     .16       0  4288.5     .05       0  4994.1     .04       0
  5000.1     .05       0  5657.9     .12       0  5787.3     .08       0
  5886.7     .05       0  6283.2     .08       0  6382.1     .05       0
Bank Sta=4883.2,5060.3
XS Rating Curve= 0 ,0
Exp/Cntr=0.3,0.1

Type RM Length L Ch R = 1 ,97461   ,197,197,197
BEGIN DESCRIPTION:
CANEY CREEK 129.0
END DESCRIPTION:
XS GIS Cut Line= 6
      3560669.43     10596219.56      3560901.17     10596224.77
      3561195.44     10596344.56      3561833.46      10596373.2
      3562500.13      10596498.2      3563446.35     10596511.17
#Sta/Elev= 30
  3896.3  416.15  3911.4  414.79  4006.5  410.13  4066.5  412.01  4124.8     407
  4128.1     407  4130.5  409.25  4153.6   409.4  4320.9  404.34  4424.3  400.59
  4708.8  393.01  4848.5  390.11  4941.6  391.78  4951.6  391.58  4998.6  377.83
  5001.4  377.33  5004.6  377.83  5011.6  385.53  5051.7   393.8  5071.7  394.94
  5176.8  391.55  5552.4   393.6  6124.9  393.65    6165  396.59  6255.1  397.35
  6408.6  409.44  6536.6     420  6665.4  433.96  6708.5  436.32  6712.2  436.41
#Mann= 10 ,-1 , 0
  3896.3     .05       0  3911.4     .16       0  4320.9     .05       0
  4424.3     .16       0  4708.8     .12       0  4848.5     .05       0
  4998.6     .04       0  5004.6     .05       0  6408.6     .12       0
  6708.5     .16       0
Bank Sta=4941.6,5071.7
XS Rating Curve= 0 ,0
Exp/Cntr=0.3,0.1

Type RM Length L Ch R = 1 ,97264   ,604,604,604
BEGIN DESCRIPTION:
CANEY CREEK 127.0
END DESCRIPTION:
XS GIS Cut Line= 3
      3560798.31     10596530.61      3562013.61     10596572.28
       3563395.1     10597002.69
#Sta/Elev= 30
    4058  432.13  4209.4  426.91  4219.4     425  4329.5  415.06  4525.1  400.99
  4621.2   394.8  4709.7  390.98  4789.7  388.91  4889.8   389.3  4969.8  391.31
  4979.8  389.17  4989.8  383.42  4996.9  376.83  4999.6  376.33  5002.9  376.83
  5009.8  377.83  5019.9   387.6  5029.9   390.5  5139.9  389.37  5918.3   390.3
  5940.2  388.87  5961.3  390.54  6044.9  390.62  6161.6  393.72  6266.6  401.83
  6505.8  422.73  6597.5   428.9    6621  429.91  6627.4  431.22    6721  434.01
#Mann= 8 ,-1 , 0
    4058     .05       0  4525.1     .16       0  4621.2     .12       0
  4996.9     .07       0  5002.9     .12       0  5009.8     .05       0
  6266.6     .12       0  6597.5     .05       0
Bank Sta=4969.8,5029.9
XS Rating Curve= 0 ,0
Exp/Cntr=0.3,0.1

Type RM Length L Ch R = 1 ,96660   ,422,422,422
BEGIN DESCRIPTION:
CANEY CREEK 126.0
END DESCRIPTION:
XS GIS Cut Line= 2
      3560888.57     10597030.61      3563228.93     10597120.89
#Sta/Elev= 30
  4298.8  435.88    4520  428.18    4656  413.25  4878.5  391.92  4930.3  387.93
  4950.3  389.15  4970.3   388.2  4990.4  377.39  4997.4  376.13  5000.1  375.63
  5003.4  376.13  5010.4  377.03  5020.4  386.88  5030.4  389.48  5104.3  388.82
  5760.9  387.06  5981.1  389.62  6021.1  387.36  6041.1  389.46  6111.2  391.09
  6184.5   395.8  6271.3  405.41  6301.3  404.33  6311.3  407.14  6331.3  409.48
  6411.4  413.25  6431.4   415.9  6551.5   422.5  6573.9  424.92  6640.9  429.79
#Mann= 8 ,-1 , 0
  4298.8     .05       0    4656     .16       0  4878.5     .12       0
  4997.4     .07       0  5003.4     .12       0  5104.3     .05       0
  6184.5     .12       0  6573.9     .05       0
Bank Sta=4950.3,5030.4
XS Rating Curve= 0 ,0
Exp/Cntr=0.3,0.1

Type RM Length L Ch R = 1 ,96238   ,454,454,454
BEGIN DESCRIPTION:
CANEY CREEK 125.0
END DESCRIPTION:
XS GIS Cut Line= 3
      3561299.63      10597360.2      3561549.61     10597460.19
      3562749.62     10597360.19
#Sta/Elev= 30
  4727.1  404.17  4813.2  396.72    4820  395.36  4920.9  387.89  4942.5  386.95
    4964  388.12  4974.8  386.01  4981.5  376.28  4983.9  375.04  4986.7  374.54
  4989.9  375.04  4998.8  375.15  5006.4  377.12  5016.4  380.86  5025.6  388.02
  5026.4  388.64  5299.9  385.75  5789.1  388.44  5819.2  388.06  5829.2   385.9
  5869.3  388.69  6009.8  387.12    6050  388.33  6090.1  391.26  6137.8  397.14
  6142.8  396.06  6150.3   398.1  6160.4  398.28  6188.6  401.84  6200.5  402.77
#Mann= 5 ,-1 , 0
  4727.1     .12       0  4983.9     .07       0  4989.9     .12       0
  5025.6     .05       0  6188.6     .12       0
Bank Sta=4964,5026.4
XS Rating Curve= 0 ,0
Exp/Cntr=0.3,0.1

Type RM Length L Ch R = 1 ,95784   ,513,513,513
BEGIN DESCRIPTION:
CANEY CREEK 124.0
END DESCRIPTION:
XS GIS Cut Line= 3
      3561199.63     10597860.19      3561399.61     10597860.19
      3563199.56      10597260.2
#Sta/Elev= 30
  4808.8  400.95  4838.8  395.96  4868.7   393.8  4978.8  386.73  4988.8  383.42
  4998.8  375.13  5003.3  374.72    5006  374.22  5009.3  374.72  5019.3  378.36
  5029.9  385.96  5040.4  387.58  5065.5  386.03    5567  387.13  5609.6  387.38
  5637.5  385.08  5651.8  387.38  5778.3  384.92  5894.2  387.85  5946.9  387.74
  5957.5  385.49  5978.5  388.14  6126.1  386.74  6326.4   394.4  6440.2  404.76
  6614.7  419.11    6727  425.44  6779.7  421.34  6821.8  430.24  6906.1  432.19
#Mann= 9 ,-1 , 0
  4808.8     .05       0  4868.7     .12       0  5003.3     .07       0
  5009.3     .12       0  5065.5     .05       0    5567     .16       0
  5637.5     .05       0  6440.2     .12       0  6614.7     .05       0
Bank Sta=4978.8,5040.4
XS Rating Curve= 0 ,0
Exp/Cntr=0.3,0.1

Type RM Length L Ch R = 1 ,95271   ,395,395,395
BEGIN DESCRIPTION:
CANEY CREEK 123.0
END DESCRIPTION:
XS GIS Cut Line= 4
      3560452.92     10598068.33      3561213.33     10598307.91
      3561494.58     10598287.07      3562905.28     10597422.95
#Sta/Elev= 30
  4056.8  420.68  4105.8  419.42  4221.2   412.2  4246.7  410.97  4284.3  406.23
    4305  406.29  4316.6  403.81  4323.6  404.68  4645.5  389.09  4818.7  385.58
  4935.8  385.98  4970.7   386.5  4980.7  385.35  5000.7  375.06  5007.8  374.37
  5010.5  373.87  5013.8  374.37  5040.8  386.43  5046.5  386.42  5501.5  385.26
  5733.7   387.1    6198  386.46  6482.3   395.5  6561.6  400.05  6571.2   402.1
  6659.1  408.31  6679.4  410.25  6766.6  419.82  6787.9  420.58  6790.4  422.05
#Mann= 9 ,-1 , 0
  4056.8     .16       0  4221.2     .12       0  4323.6     .05       0
  4935.8     .16       0  5007.8     .07       0  5013.8     .16       0
  5046.5     .05       0  6659.1     .12       0  6679.4     .05       0
Bank Sta=4970.7,5040.8
XS Rating Curve= 0 ,0
Exp/Cntr=0.3,0.1

Type RM Length L Ch R = 1 ,94876   ,454,454,454
BEGIN DESCRIPTION:
CANEY CREEK 122.0
END DESCRIPTION:
XS GIS Cut Line= 3
      3560825.05      10599375.3      3561399.61     10598610.19
      3562599.59      10597710.2
#Sta/Elev= 30
  4056.7  411.82  4085.6  411.48  4106.4  407.56  4277.9  391.67  4435.5  383.22
  4441.7   376.7  4450.1  375.11  4477.2  384.31  4576.6  383.66  4634.2  383.59
  4814.9  382.97    4950  385.89  4956.2  385.79  4963.5     376  4988.7  372.99
  4991.4  372.49  4994.7  372.99  5006.2  373.05  5010.4  375.52  5020.8  373.85
  5027.1  381.37  5035.4  380.49  5041.6     384  5063.5  385.27  5210.5  384.86
  5474.7  384.38  5481.1   384.3  6306.2  386.87  6427.1  389.68  6513.5  394.68
#Mann= 10 ,-1 , 0
  4056.7     .16       0  4277.9     .12       0  4576.6     .16       0
  4634.2     .05       0  4814.9     .16       0  4988.7     .07       0
  4994.7     .16       0  5210.5     .05       0  5474.7     .08       0
  5481.1     .05       0
Bank Sta=4950,5063.5
XS Rating Curve= 0 ,0
Exp/Cntr=0.3,0.1

Type RM Length L Ch R = 1 ,94422   ,463,463,463
BEGIN DESCRIPTION:
CANEY CREEK 121.0
END DESCRIPTION:
XS GIS Cut Line= 3
      3560809.85     10599488.15      3561599.61     10598960.19
      3562799.58     10597760.22
#Sta/Elev= 30
  4048.9  407.34  4198.6  402.32  4249.6  395.63  4411.8  385.14  4516.9  383.73
  4522.9  375.64  4529.8  373.57  4537.9  374.73  4552.9  383.14  4635.7  382.33
  4688.1  380.43  4712.5  382.28  4855.5  383.72  4970.4  385.03  4976.4  383.79
  4992.9  372.83  4995.6  372.33  4998.9  372.83  5002.4  372.83    5013  382.54
  5027.2  384.86  5253.4  384.17  5338.3  382.93  5366.6  380.13  5435.8  383.32
    5508  388.06  5875.7  392.27  6059.5  390.27  6413.1  392.91  6695.9  406.56
#Mann= 8 ,-1 , 0
  4048.9     .16       0  4411.8     .12       0  4635.7     .05       0
  4712.5     .07       0  4855.5     .12       0  4992.9     .07       0
  4998.9     .12       0  5435.8     .05       0
Bank Sta=4970.4,5027.2
XS Rating Curve= 0 ,0
Exp/Cntr=0.3,0.1

Type RM Length L Ch R = 1 ,93959   ,516,516,516
BEGIN DESCRIPTION:
CANEY CREEK 120.0
END DESCRIPTION:
XS GIS Cut Line= 3
      3561499.59     10599760.22      3561949.61     10599160.19
      3563149.61     10597960.18
#Sta/Elev= 30
  4217.2  401.45    4387  387.95  4395.4  387.98  4495.4  382.23  4503.7  379.67
  4509.9  381.59  4527.8  371.72  4530.5  371.22  4533.8  371.72  4545.4  381.64
  4609.1  380.74  4853.2  383.35  4939.1  382.43  4945.4  378.55  4970.8  379.52
  4981.4  375.02  5009.7  373.42  5023.8  376.87  5037.9  384.14  5052.1  384.28
  5132.7  383.51  5660.2  383.22  5992.3  386.95  5997.5  387.12  6130.9  390.92
  6137.9  391.03  6264.4  397.97  6297.7  400.43  6379.9   403.9  6664.3   426.3
#Mann= 14 ,-1 , 0
  4217.2     .16       0    4387     .12       0  4527.8     .07       0
  4533.8     .12       0  4609.1     .07       0  4853.2     .12       0
  5132.7     .05       0  5992.3      .1       0  5997.5     .08       0
  6130.9     .05       0  6137.9      .1       0  6264.4     .05       0
  6297.7     .08       0  6379.9     .05       0
Bank Sta=4395.4,5052.1
XS Rating Curve= 0 ,0
Exp/Cntr=0.3,0.1
