HEC-RAS study COTTONWOOD CREEK.prj: COTTONWOOD CREEK Base Level Engineering

--- COTTONWOOD CREEK.g01 (geometry) --- (continued)

Type RM Length L Ch R = 1 ,69743   ,461,461,461
BEGIN DESCRIPTION:
COTTONWOOD CREEK 73.0
END DESCRIPTION:
XS GIS Cut Line= 2
      3582941.92     10647182.11      3586353.42     10647616.14
#Sta/Elev= 30
  3066.8  354.17    3125  354.11  3336.6  334.31  3598.7  315.79  4219.7  315.38
    4254  312.97  4376.1  315.59  4385.9  315.61  4455.6  315.72  4485.8  312.22
  4556.4  316.46  4576.6  312.15  4594.2  314.56  4599.2  311.52  4674.1  312.72
  4687.4  316.99  4959.6  316.42  4979.8  305.84  4996.9  303.51  4999.7  303.01
  5002.9  303.51  5020.1  316.62  5050.4  319.33  5080.6  315.25  5226.1  315.79
  5263.8   315.7  5461.7  316.33  5875.3  323.33  6117.9  336.03  6505.8  354.52
#Mann= 11 ,-1 , 0
  3066.8     .05       0  4219.7     .12       0  4376.1     .16       0
  4385.9     .12       0  4996.9     .07       0  5002.9     .12       0
  5226.1     .05       0  5263.8     .12       0  5461.7     .16       0
  5875.3     .12       0  6117.9     .16       0
Bank Sta=4959.6,5020.1
XS Rating Curve= 0 ,0
Exp/Cntr=0.3,0.1

Type RM Length L Ch R = 1 ,69282   ,445,445,445
BEGIN DESCRIPTION:
COTTONWOOD CREEK 72.0
END DESCRIPTION:
XS GIS Cut Line= 2
      3582325.61     10647685.58      3585875.28     10647919.91
#Sta/Elev= 30
  2477.5  353.67  2651.9  347.08  2671.9   342.9  2752.1   343.3  2832.3  336.87
  2949.6  340.44  3273.2  336.43  3503.7  316.03  3580.5  315.48  3606.6  315.89
  4433.1  313.57  4526.7   315.3    4546  312.35  4696.3   315.3  4716.4  312.35
  4736.4  315.46  4966.9  316.05  4976.9  314.38  4986.9  306.56    5004  303.35
  5006.7  302.85    5010  303.35    5017  303.88    5027  314.96  5037.1   316.1
  5250.4  314.08  5373.2  314.38  5697.6  329.07  5856.4  340.63  6034.9  352.71
#Mann= 12 ,-1 , 0
  2477.5     .12       0  2949.6     .05       0  3580.5     .16       0
  3606.6     .05       0  4433.1      .1       0  4526.7     .12       0
    5004     .07       0    5010     .12       0  5250.4     .05       0
  5373.2     .16       0  5697.6     .05       0  5856.4     .16       0
Bank Sta=4966.9,5037.1
XS Rating Curve= 0 ,0
Exp/Cntr=0.3,0.1

Type RM Length L Ch R = 1 ,68837   ,846,846,846
BEGIN DESCRIPTION:
COTTONWOOD CREEK 71.0
END DESCRIPTION:
XS GIS Cut Line= 3
       3582490.5     10648050.16      3584400.25     10648353.98
      3585849.95     10648058.83
#Sta/Elev= 30
  2607.3  359.11  2884.8  335.63  2956.6  326.85  2998.4  326.54  3051.9  329.13
  3193.7  323.34  3396.2  323.48  3639.2  313.27  3892.4   315.2    4024  312.34
  4034.1  309.09  4296.1  312.65    4969   315.1  4979.2  312.75  4985.2  304.17
  4996.6  303.07  4999.4  302.57  5002.6  303.07  5003.1  303.09  5020.1  305.02
  5035.8  315.22  5097.8  313.98  5104.9  313.71  5435.3   318.5  5530.3  323.84
    5587  332.39  5673.2  330.59  5797.4  336.81  5826.3  344.49  6020.5  353.29
#Mann= 10 ,-1 , 0
  2607.3     .12       0  2884.8     .16       0  2998.4     .05       0
  4296.1     .12       0  4996.6     .07       0  5002.6     .12       0
  5003.1     .05       0  5097.8     .12       0  5104.9     .05       0
  5797.4     .16       0
Bank Sta=4969,5035.8
XS Rating Curve= 0 ,0
Exp/Cntr=0.3,0.1

Type RM Length L Ch R = 1 ,67991   ,511,511,511
BEGIN DESCRIPTION:
COTTONWOOD CREEK 70.0
END DESCRIPTION:
XS GIS Cut Line= 3
      3583149.56     10649760.21      3584949.61     10648960.19
       3585599.6      10648360.2
#Sta/Elev= 30
  3059.4   344.1    3102  341.06  3127.9  338.93  3238.1  329.98  3348.3  320.69
  3415.8  315.64  3568.7  314.87  3789.1  314.83  3861.7  314.35    3885  309.09
  3908.2  314.12  4066.2  313.21    4082  309.09  4110.7  313.09  4320.1  311.57
  4897.9  312.18  4974.5  313.85  4994.1  301.14  4996.8  300.64  5000.1  301.14
  5026.5   314.3  5057.3   314.3  5071.5     310  5078.8  314.26  5269.9  312.26
  5456.3   320.7  5648.8   333.4  5692.4  336.34  5904.7  349.45  5913.8  349.45
#Mann= 15 ,-1 , 0
  3059.4     .16       0    3102     .12       0  3127.9     .16       0
  3238.1     .12       0  3348.3     .16       0  3568.7     .05       0
  3789.1     .12       0  4320.1     .05       0  4897.9     .12       0
  4994.1     .07       0  5000.1     .12       0  5456.3     .16       0
  5648.8     .05       0  5692.4     .16       0  5904.7     .05       0
Bank Sta=4974.5,5026.5
XS Rating Curve= 0 ,0
Exp/Cntr=0.3,0.1

Type RM Length L Ch R = 1 ,67480   ,1716,1716,1716
BEGIN DESCRIPTION:
COTTONWOOD CREEK 69.0
END DESCRIPTION:
XS GIS Cut Line= 3
      3583149.65     10649810.18      3585149.61     10649410.19
      3585949.57     10648960.21
#Sta/Elev= 30
  2947.6  346.89  3008.7  342.65  3110.4  335.06  3212.1  327.22  3416.7  314.92
  3720.6  312.15  4242.7  312.38  4273.3  308.59  4314.1  307.92  4375.3  308.86
  4405.9  312.23  4487.5  312.38  4497.7  309.76  4528.3  312.32  4599.6  311.38
  4609.8  305.03  4630.2  311.15  4640.4  311.48    4824  310.53  4966.8  312.75
    4990  308.33  4995.1  301.41  4997.9  301.33  5000.6  300.83  5003.9  301.33
  5010.1  301.89  5016.8  312.79    5274  310.54  5528.1  320.43    5905  342.36
#Mann= 8 ,-1 , 0
  2947.6     .16       0  3008.7     .12       0  3110.4     .16       0
  3212.1     .05       0  3720.6     .12       0  4997.9     .07       0
  5003.9     .12       0  5528.1     .16       0
Bank Sta=4966.8,5016.8
XS Rating Curve= 0 ,0
Exp/Cntr=0.3,0.1

Type RM Length L Ch R = 1 ,65764   ,795,795,795
BEGIN DESCRIPTION:
COTTONWOOD CREEK 68.0
END DESCRIPTION:
XS GIS Cut Line= 3
      3583545.22     10651532.51       3586453.2     10649848.48
        3586748.     10648834.05
#Sta/Elev= 30
  1819.6   354.8  1986.4  351.15  2036.1  344.57  2073.4  345.48  2271.4  332.86
  2871.2   321.9  3122.1  311.93  3176.8  309.16  3229.9  311.83  3257.2   310.5
  3535.7  308.31  4735.1  309.91  4948.8  310.61  4964.6  312.98  4979.4  308.79
  4986.1  300.44  4988.9  299.61  4991.6  299.11  4994.9  299.61  5007.6   301.2
  5014.1  307.21  5023.4  310.98  5086.1  310.21  5358.7  310.85  5401.1  310.52
  5480.2  317.67  5623.8  322.44  5935.4  337.88  6125.9   343.6  6236.4  343.79
#Mann= 10 ,-1 , 0
  1819.6     .05       0  3122.1     .08       0  3257.2      .1       0
  3535.7     .05       0  4735.1     .12       0  4988.9     .07       0
  4994.9     .12       0  5086.1     .05       0  5358.7     .12       0
  5623.8     .16       0
Bank Sta=4964.6,5023.4
XS Rating Curve= 0 ,0
Exp/Cntr=0.3,0.1

Type RM Length L Ch R = 1 ,64969   ,1258,1258,1258
BEGIN DESCRIPTION:
COTTONWOOD CREEK 67.0
END DESCRIPTION:
XS GIS Cut Line= 3
      3584649.64     10652010.16      3586249.61     10650460.19
      3587799.59      10649160.2
#Sta/Elev= 30
    2754  367.38  2923.6  361.89  3157.2  349.79    3348  346.92  3397.4  338.04
  3524.8  335.93  3837.7  311.97  3910.3  310.96  4281.6  305.69  4288.5  304.35
  4302.7  305.82  4858.4  307.59  4974.6   309.7  4978.1  300.39  4983.2  300.39
  4992.3  298.44  4995.1  297.94  4998.3  298.44  5003.1  298.79  5009.6  304.42
  5023.9  309.82  5116.8  308.75  5140.5  308.67  5634.2  308.44  6365.2  317.91
  6486.2  321.87  6564.3  327.66  6798.4  355.18    6870  358.66  7004.6  360.71
#Mann= 9 ,-1 , 0
    2754     .05       0  3837.7     .16       0  3910.3     .05       0
  4858.4     .12       0  4983.2     .16       0  4992.3     .07       0
  4998.3     .16       0  5116.8     .12       0  5140.5     .05       0
Bank Sta=4974.6,5023.9
XS Rating Curve= 0 ,0
Exp/Cntr=0.3,0.1

Type RM Length L Ch R = 1 ,63711   ,907,907,907
BEGIN DESCRIPTION:
COTTONWOOD CREEK 66.0
END DESCRIPTION:
XS GIS Cut Line= 3
      3586249.62     10651610.16      3586549.61     10651060.19
      3587949.59     10649610.21
#Sta/Elev= 30
  4374.7   340.4  4477.2  331.87  4529.9  322.03  4573.5  317.21  4655.2  314.48
  4750.6   315.5  4830.3  306.06  4901.5  308.43  4965.6   306.5  4971.3     308
  4978.4     301  4993.1  300.86  4998.3  298.16  5005.2  297.93    5008  297.43
  5011.2  297.93  5019.9  298.08  5029.3     298  5043.5  306.66  5050.7  308.55
  5213.3  305.22  5291.2  306.61  5800.3   305.4  5969.9  307.53  6010.4   308.8
  6150.7  310.81  6472.3  317.18  6889.5  352.96  6946.1  356.13  7016.7  357.01
#Mann= 8 ,-1 , 0
  4374.7     .05       0  4901.5     .16       0  5005.2     .07       0
  5011.2     .16       0  5019.9     .05       0  5969.9     .16       0
  6010.4     .05       0  6150.7     .16       0
Bank Sta=4971.3,5050.7
XS Rating Curve= 0 ,0
Exp/Cntr=0.3,0.1

Type RM Length L Ch R = 1 ,62804   ,617,617,617
BEGIN DESCRIPTION:
COTTONWOOD CREEK 65.0
END DESCRIPTION:
XS GIS Cut Line= 3
      3586378.05     10651826.79      3587207.05     10651241.71
      3588126.26     10650084.03
#Sta/Elev= 30
  4121.5  345.74  4221.3  341.43  4644.1  304.72  4679.8  307.48  4761.9  307.53
  4765.6  307.48  4900.9  305.88  4967.9  306.24  4980.2  304.07  5000.6  295.71
  5003.4  295.21  5006.6  295.71  5016.9  297.18  5024.6  304.84  5030.7  306.46
  5351.9  305.14  5787.3  309.11  5942.6  320.23  6134.9  328.36  6192.6  326.35
  6224.1   329.4  6242.2   330.6  6256.7  325.88  6277.5  326.24  6312.9  327.87
  6335.2  333.62  6376.8  335.47  6391.2  332.74  6405.7  336.41  6614.4  344.75
#Mann= 8 ,-1 , 0
  4121.5     .05       0  4761.9     .16       0  4765.6     .05       0
  4900.9     .12       0  5000.6     .07       0  5006.6     .12       0
  5351.9     .05       0  6224.1     .16       0
Bank Sta=4967.9,5030.7
XS Rating Curve= 0 ,0
Exp/Cntr=0.3,0.1

Type RM Length L Ch R = 1 ,62187   ,883,883,883
BEGIN DESCRIPTION:
COTTONWOOD CREEK 64.0
END DESCRIPTION:
XS GIS Cut Line= 3
      3586329.44     10652007.34      3587197.51     10651903.17
      3588322.51      10650361.5
#Sta/Elev= 30
  3959.7  345.87  4110.9  344.39  4145.9  342.61  4219.1  335.48  4478.3  312.68
  4567.2  307.06  4719.8  304.67  4973.9  306.38  4987.1  299.93  4992.6  295.28
  4995.3  294.78  4998.6  295.28  5016.4  296.02  5023.4  302.46  5031.1  306.27
    5096  305.65  5102.2  304.45  5116.8  305.38    5123  303.97  5131.5  305.27
  5309.2  303.62  5461.5  304.89  5811.2  308.51  6097.8  314.34  6192.9  318.45
  6325.7  325.76  6419.9  333.76  6583.2  343.02  6626.1   344.1  6742.5  348.16
#Mann= 9 ,-1 , 0
  3959.7     .05       0  4219.1     .16       0  4478.3     .05       0
  4719.8     .12       0  4992.6     .07       0  4998.6     .12       0
  5461.5     .05       0  6192.9     .16       0  6626.1     .05       0
Bank Sta=4973.9,5031.1
XS Rating Curve= 0 ,0
Exp/Cntr=0.3,0.1

Type RM Length L Ch R = 1 ,61304   ,749,749,749
BEGIN DESCRIPTION:
COTTONWOOD CREEK 63.0
END DESCRIPTION:
XS GIS Cut Line= 2
      3586627.71     10652359.94      3589120.83     10651602.98
#Sta/Elev= 30
  3731.3  341.05  3764.6  340.45  3827.3  328.79  3900.5     325  3986.3  315.85
  4090.9  309.33  4109.8  308.58  4339.4  302.64  4517.1  304.98    4607  303.17
  4788.8   305.5  4984.5  305.14  4989.7   304.5  4997.8  295.93  5005.3  295.03
    5008  294.53  5011.3  295.03  5017.4  295.44  5029.2  302.99  5039.6  305.33
  5137.5  303.41  5440.9  304.94  5556.1  307.23  5914.2  330.46  6091.5  334.38
  6116.1  335.85    6122  339.03  6127.2  337.54  6155.1   340.1  6336.8   340.9
#Mann= 11 ,-1 , 0
  3731.3     .05       0  3986.3     .16       0  4090.9     .05       0
  4109.8     .12       0  5005.3     .07       0  5011.3     .12       0
  5137.5     .05       0  5440.9     .16       0  5556.1     .05       0
  6091.5     .08       0  6155.1     .05       0
Bank Sta=4984.5,5039.6
XS Rating Curve= 0 ,0
Exp/Cntr=0.3,0.1

Type RM Length L Ch R = 1 ,60555   ,283,283,283
BEGIN DESCRIPTION:
COTTONWOOD CREEK 62.0
END DESCRIPTION:
XS GIS Cut Line= 2
      3586551.37     10652901.59      3588801.32     10652075.22
#Sta/Elev= 30
  3870.2  338.88  3972.7   338.6  4058.8  334.66    4156  324.21  4251.8  318.04
    4292   313.9  4297.3  311.16    4350  312.74  4404.2  309.64  4618.1  303.34
    4832  302.99  4843.7  303.17  4961.1  304.95  4988.6  294.75  4991.3  294.25
  4994.6  294.75  5008.2  295.11  5016.8  297.74  5022.1  302.14  5040.2  304.52
    5072  304.08  5511.6  303.49  5618.5  305.94  5817.8   312.1  5858.1  316.19
  5863.5   314.6  5998.3  322.76  6041.6  324.51  6207.9  340.22  6267.1  341.18
#Mann= 13 ,-1 , 0
  3870.2     .16       0  4297.3     .12       0    4350     .16       0
  4404.2     .05       0  4618.1     .16       0    4832     .05       0
  4843.7     .12       0  4988.6     .07       0  4994.6     .12       0
    5072     .05       0  5511.6     .16       0  5618.5     .05       0
  5998.3     .12       0
Bank Sta=4961.1,5040.2
XS Rating Curve= 0 ,0
Exp/Cntr=0.3,0.1

Type RM Length L Ch R = 1 ,60272   ,1034,1034,1034
BEGIN DESCRIPTION:
COTTONWOOD CREEK 61.0
END DESCRIPTION:
XS GIS Cut Line= 2
      3586704.16     10653234.92      3588695.91     10652298.03
#Sta/Elev= 30
  3856.5   345.9  3891.8  342.27  3924.5  337.76  4018.4  328.54  4157.5   314.4
  4186.4  311.53  4314.9  304.93  4729.4  301.87  4983.9  303.87  4989.7  303.78
  4997.8  294.89  5000.5  294.39  5003.8  294.89  5022.9  295.04  5029.5  299.64
    5045  303.92  5155.5  303.22  5177.6  300.68  5201.7  302.09  5222.9  299.94
  5236.8   301.9  5336.9  304.79  5428.1  309.89  5450.9  309.47  5570.4  316.84
  5614.7  317.72  5712.7  321.45  5758.3  325.34  5877.8  328.41  6057.6  340.08
#Mann= 13 ,-1 , 0
  3856.5     .05       0  3891.8     .16       0  3924.5     .12       0
  4018.4     .16       0  4157.5     .05       0  4186.4     .16       0
  4314.9     .05       0  4729.4     .12       0  4997.8     .07       0
  5003.8     .12       0  5201.7     .05       0  5236.8     .16       0
  5614.7     .12       0
Bank Sta=4983.9,5045
XS Rating Curve= 0 ,0
Exp/Cntr=0.3,0.1

Type RM Length L Ch R = 1 ,59238   ,366,366,366
BEGIN DESCRIPTION:
COTTONWOOD CREEK 60.0
END DESCRIPTION:
XS GIS Cut Line= 3
       3586919.4     10653540.48      3588051.35     10653540.48
      3588620.32     10652444.19
#Sta/Elev= 30
  3707.7  336.96  3947.9  319.98    4099  313.42  4204.4  308.07  4387.9  301.04
  4501.2  300.66  4600.2  301.17  4677.9  299.51  4717.9  301.57  4890.4  301.02
  4963.9  303.25  4978.9  297.19    4998  293.44  5000.8  292.94    5004  293.44
  5017.5  303.73  5089.5  301.31  5166.7  300.97  5188.8  298.74  5200.5  300.74
  5223.1  299.72  5296.7  301.48  5476.4  300.95  5625.4  305.24  5707.5  310.74
  5790.4  318.95  5876.5   327.7  5935.3  335.71  5979.6  338.82  6074.8  337.73
#Mann= 10 ,-1 , 0
  3707.7     .12       0    4099     .16       0  4204.4     .05       0
  4501.2     .16       0  4600.2     .12       0    4998     .07       0
    5004     .12       0  5296.7     .05       0  5625.4     .16       0
  5790.4     .12       0
Bank Sta=4963.9,5017.5
XS Rating Curve= 0 ,0
Exp/Cntr=0.3,0.1

Type RM Length L Ch R = 1 ,58872   ,393,393,393
BEGIN DESCRIPTION:
COTTONWOOD CREEK 59.0
END DESCRIPTION:
XS GIS Cut Line= 3
      3588315.24     10654290.52      3588322.19     10653471.04
      3588676.34     10652561.36
#Sta/Elev= 30
  4360.1  334.39  4420.4  335.64  4510.4   332.1  4610.4  322.35  4760.4  310.98
  4820.4  303.66  4882.2  300.27  4910.5  298.76  4920.5   300.4  4930.5  299.72
  4950.5  301.95  4970.5   302.1  4980.5  299.05  4987.5  292.76  4990.2  292.26
  4993.5  292.76  5000.5  292.88  5010.5  300.88  5020.5   302.9  5270.4  301.49
  5277.1  298.23  5287.8  302.26    5493  300.15  5695.6   302.3  5781.5  304.68
  5874.7  309.96  5903.9  312.19  5928.4  316.53  5984.6  321.31  6155.8  340.81
#Mann= 7 ,-1 , 0
  4360.1     .16       0  4882.2     .12       0  4987.5     .07       0
  4993.5     .12       0    5493     .05       0  5874.7     .16       0
  5984.6     .12       0
Bank Sta=4970.5,5020.5
XS Rating Curve= 0 ,0
Exp/Cntr=0.3,0.1

Type RM Length L Ch R = 1 ,58479   ,562,562,562
BEGIN DESCRIPTION:
COTTONWOOD CREEK 58.0
END DESCRIPTION:
XS GIS Cut Line= 3
      3588349.61     10654160.19      3588549.61     10653410.19
       3588749.6     10652610.21
#Sta/Elev= 30
  4223.6  335.17  4321.3  328.34  4347.8  324.97  4378.8  323.46    4503  311.71
  4596.8  305.92  4623.6  299.89  4631.8  298.79    4679  301.65    4787  302.59
  4968.8   301.9  4977.2  295.44  4982.3  295.28  4986.5   292.7  4989.2   292.2
  4992.5   292.7  5002.4  292.88  5010.1  299.02  5017.8  301.19  5105.5  300.46
  5123.5  298.18  5133.8  299.89    5175  301.37  5275.7  302.92  5471.4  305.66
  5600.2  312.16  5620.7  314.39  5636.3  317.06  5668.3  319.58  5824.4  335.97
#Mann= 7 ,-1 , 0
  4223.6     .16       0  4623.6     .12       0  4986.5     .07       0
  4992.5     .12       0  5275.7     .05       0  5620.7     .16       0
  5668.3     .12       0
Bank Sta=4968.8,5017.8
XS Rating Curve= 0 ,0
Exp/Cntr=0.3,0.1

Type RM Length L Ch R = 1 ,57917   ,702,702,702
BEGIN DESCRIPTION:
COTTONWOOD CREEK 57.0
END DESCRIPTION:
XS GIS Cut Line= 3
      3588399.64     10654110.16      3589049.61     10653610.19
      3589549.64     10652910.15
#Sta/Elev= 30
  4178.8  332.45  4300.2  320.43  4337.2  318.87    4485  310.16  4506.8  307.54
    4514  304.89  4557.2  303.64  4592.9  301.81  4613.7  302.73  4670.8  299.14
  4707.1  299.68  4727.9  298.32  4734.2  299.63  4935.4  303.27  4970.7  301.35
  4977.1  293.74  4988.6  292.11  4991.3  291.61  4994.6  292.11  5001.9  292.16
  5006.2  295.66  5012.3  296.56  5020.9  302.09  5071.3  299.95  5113.2  299.87
  5249.5  300.88  5350.3  305.37  5658.7  328.72  5786.5  340.95  5859.1  344.89
#Mann= 6 ,-1 , 0
  4178.8     .16       0  4337.2     .05       0  4557.2     .12       0
  4988.6     .07       0  4994.6     .12       0  5113.2     .05       0
Bank Sta=4970.7,5020.9
XS Rating Curve= 0 ,0
Exp/Cntr=0.3,0.1

Type RM Length L Ch R = 1 ,57215   ,543,543,543
BEGIN DESCRIPTION:
COTTONWOOD CREEK 56.0
END DESCRIPTION:
XS GIS Cut Line= 3
      3588399.61     10654160.19      3589049.61     10654060.19
      3589849.57     10653560.21
#Sta/Elev= 30
  4356.9  335.79  4407.5  329.97  4427.7   325.6  4499.9  319.21  4585.8  309.94
  4670.5  304.46  4751.5  301.83  4761.6  300.33  4776.8  299.81  4862.8  300.59
    4883  299.21  4923.5  300.14    4964  299.67  4974.1  300.79  4985.5  299.87
  4994.3  292.07  5001.4  291.17  5004.2  290.67  5007.4  291.17  5017.5  291.22
  5028.1  292.77  5037.5  301.18  5190.9  299.96  5311.1   300.8  5472.7  300.31
  5609.5  303.43  5688.5  308.09  5740.4  312.93  5828.2  318.92  5957.9  331.91
#Mann= 6 ,-1 , 0
  4356.9     .16       0  4499.9     .05       0  4776.8     .12       0
  5001.4     .07       0  5007.4     .12       0  5190.9     .05       0
Bank Sta=4985.5,5037.5
XS Rating Curve= 0 ,0
Exp/Cntr=0.3,0.1

Type RM Length L Ch R = 1 ,56672   ,672,672,672
BEGIN DESCRIPTION:
COTTONWOOD CREEK 55.0
END DESCRIPTION:
XS GIS Cut Line= 3
      3588112.75     10655460.21      3589420.06     10654397.69
      3589841.94     10653689.35
#Sta/Elev= 30
  3430.7  346.96  3720.3  319.82  3819.4  313.86  3897.7  306.96  3968.1  302.78
  4084.2  301.63  4215.9  301.41  4266.6  300.14  4558.9   298.7  4586.5  297.43
  4600.9  294.78  4608.8  298.94  4615.3  299.23    4857  298.24  4907.7   300.9
  4971.6  301.25    4978  299.57  4985.9  294.55  4992.4  293.38  4995.8  290.62
  4998.6  290.12  5001.8  290.62  5013.2  292.54  5027.6  299.38  5109.8  300.06
  5493.1  301.75  5689.8  310.64  5732.6  314.76  5799.1  317.39  5939.8  326.55
#Mann= 8 ,-1 , 0
  3430.7     .05       0  4084.2     .16       0  4215.9     .05       0
  4266.6     .16       0  4558.9     .12       0  4995.8     .07       0
  5001.8     .12       0  5109.8     .05       0
Bank Sta=4971.6,5027.6
XS Rating Curve= 0 ,0
Exp/Cntr=0.3,0.1

Type RM Length L Ch R = 1 ,56000   ,111,111,111
BEGIN DESCRIPTION:
COTTONWOOD CREEK 54.0
END DESCRIPTION:
XS GIS Cut Line= 2
      3589451.31     10655850.81       3589753.4     10654397.68
#Sta/Elev= 30
  4123.2  329.66  4201.1  323.97  4239.5  321.92  4300.4  316.09  4499.1  302.07
  4598.4  297.81  4630.1  296.61  4635.2  297.61  4680.2  297.62  4697.8  295.73
  4730.3  296.23  4736.7  297.71  4757.1  296.12  4808.2  299.57    4849  300.54
  4896.5  299.83  4975.7  300.58    4992  290.59  4999.2  290.18    5002  289.68
  5005.2  290.18  5012.4  297.89  5030.7  297.63  5095.1  299.23  5380.1  312.17
  5511.5  314.47  5523.1  315.89  5561.6  315.66  5566.7  316.73  5607.4  315.82
#Mann= 11 ,-1 , 0
  4123.2     .05       0  4201.1     .08       0  4300.4     .05       0
  4499.1     .08       0  4598.4      .1       0  4697.8     .08       0
  4896.5     .12       0  4999.2     .07       0  5005.2     .12       0
  5030.7     .08       0  5095.1     .05       0
Bank Sta=4975.7,5012.4
XS Rating Curve= 0 ,0
Exp/Cntr=0.3,0.1

Type RM Length L Ch R = 1 ,55889   ,1120,1120,1120
BEGIN DESCRIPTION:
COTTONWOOD CREEK 53.0
END DESCRIPTION:
XS GIS Cut Line= 2
      3589539.84     10655892.52      3589836.57     10654424.51
#Sta/Elev= 30
  4157.7  325.13  4285.2   319.3  4330.8  318.81  4455.9  305.29  4567.9  298.12
  4670.2  296.94  4772.2  298.82  4782.4  296.26  4787.5  298.41  4869.7  298.25
  4945.7  299.65  4955.9  296.06  4976.3  292.38  4985.3  292.87  4993.7  289.78
  4996.4  289.28  4999.7  289.78  5036.1  290.29  5047.7  294.78  5068.2  297.71
  5078.3  298.65  5151.2  303.64  5167.5   304.4  5193.4  307.97  5289.8  311.42
  5396.4  318.34  5492.8  320.88  5497.9  324.02  5537.4  321.29  5655.4  323.33
#Mann= 8 ,-1 , 0
  4157.7     .05       0  4567.9     .12       0  4869.7     .05       0
  4993.7     .04       0  4999.7     .05       0  5068.2     .08       0
  5151.2     .12       0  5167.5     .05       0
Bank Sta=4945.7,5078.3
XS Rating Curve= 0 ,0
Exp/Cntr=0.3,0.1

Type RM Length L Ch R = 1 ,54769   ,896,896,896
BEGIN DESCRIPTION:
COTTONWOOD CREEK 52.0
END DESCRIPTION:
XS GIS Cut Line= 3
      3590644.02      10656623.4      3590461.73     10655573.04
      3590505.13     10654297.03
#Sta/Elev= 30
  4046.5  333.69  4065.1  333.24  4158.2  330.15  4163.2   331.4  4243.8  327.27
  4303.5  324.93  4486.2  309.07    4636  299.75  4831.3  295.55  4973.4  300.28
  4983.7  294.03  5000.8  289.92  5003.6  289.42  5006.8  289.92  5033.2  299.24
  5111.5  296.11  5315.5  297.77  5415.6  305.45  5505.6  307.27  5575.7  305.92
  5605.4  301.52  5635.7  305.98  5665.7  303.87  5705.8  307.05  5885.9  310.75
    6066  322.75  6080.4  322.24    6096  325.27    6176  330.34  6389.3  338.68
#Mann= 7 ,-1 , 0
  4046.5     .12       0  4065.1     .16       0  4243.8     .05       0
    4636     .12       0  5000.8     .07       0  5006.8     .12       0
  5605.4     .05       0
Bank Sta=4973.4,5033.2
XS Rating Curve= 0 ,0
Exp/Cntr=0.3,0.1

Type RM Length L Ch R = 1 ,53873   ,616,616,616
BEGIN DESCRIPTION:
COTTONWOOD CREEK 51.0
END DESCRIPTION:
XS GIS Cut Line= 3
      3590999.61     10656460.19      3590999.61     10655860.19
      3591049.61     10654560.15
#Sta/Elev= 30
  4380.6   328.2  4500.6  318.07  4530.6  316.88  4540.6  314.75  4620.6  308.17
  4711.9  302.62  4857.2  296.91  4890.6  295.42  4970.6  298.74  4978.1   296.5
  4983.1   296.5  4990.6  289.18  4997.6  288.49  5000.4  287.99  5003.6  288.49
  5010.6  289.33  5020.6  296.84  5030.6  298.38  5120.7  296.82  5180.8  297.68
  5380.9  296.34  5440.9  298.78  5527.8  299.26  5741.2  303.19  5831.2  307.86
  5959.2  316.81    6078  326.23    6106  328.88  6221.5  338.35  6281.6  339.62
#Mann= 9 ,-1 , 0
  4380.6     .05       0  4711.9     .16       0  4857.2     .12       0
  4997.6     .07       0  5003.6     .12       0  5527.8     .16       0
  5959.2     .12       0    6078     .16       0    6106     .12       0
Bank Sta=4970.6,5030.6
XS Rating Curve= 0 ,0
Exp/Cntr=0.3,0.1

Type RM Length L Ch R = 1 ,53257   ,494,494,494
BEGIN DESCRIPTION:
COTTONWOOD CREEK 50.0
END DESCRIPTION:
XS GIS Cut Line= 2
      3591462.46     10656498.36      3591580.52      10654685.8
#Sta/Elev= 30
  4226.6  322.62    4355  312.88  4435.2  308.96  4545.4  301.65  4577.8  300.69
  4688.4  298.04  4765.9  295.62    4826  296.55  4846.1  294.97  4878.1  296.27
  4956.3  297.02  4976.4  298.84  4986.4  289.38  4993.4  287.88  4996.2  287.38
  4999.4  287.88  5006.4  288.42  5016.4  296.89  5182.3  298.07    5297  296.71
  5377.2  296.96  5547.6  300.41  5657.8  305.81    5758  313.86  5858.2  324.32
  5888.3  326.01  5898.3  327.88  5925.5   328.8  5978.5  332.04    6043   332.1
#Mann= 6 ,-1 , 0
  4226.6     .05       0  4577.8     .16       0  4688.4     .12       0
  4993.4     .07       0  4999.4     .12       0  5925.5      .1       0
Bank Sta=4976.4,5016.4
XS Rating Curve= 0 ,0
Exp/Cntr=0.3,0.1

Type RM Length L Ch R = 1 ,52763   ,975,975,975
BEGIN DESCRIPTION:
COTTONWOOD CREEK 49.0
END DESCRIPTION:
XS GIS Cut Line= 2
      3591858.29     10656567.81      3592316.34     10653923.59
#Sta/Elev= 30
  4203.1  320.64  4231.1  320.59  4271.7  317.57    4303  317.97  4312.3  315.97
  4373.2  312.78  4586.3  307.14  4656.6  302.45  4809.4  293.27  4931.4  297.07
    4972  296.36  4982.2  288.13  4989.3  286.46  4992.1  285.96  4995.3  286.46
  5004.6  286.92  5012.6  292.85  5022.8  297.69  5043.1  296.28  5225.7  296.39
  5367.8  298.85    5806  301.73  5896.6  302.38  6228.7  303.94  6372.6  302.18
  6390.9  303.39  6489.7  311.93  6606.2  322.85  6768.4  337.95  6886.7   337.1
#Mann= 10 ,-1 , 0
  4203.1     .05       0  4656.6     .16       0  4809.4     .12       0
  4989.3     .07       0  4995.3     .12       0    5806     .16       0
  5896.6     .12       0  6390.9     .05       0  6489.7     .16       0
  6606.2     .12       0
Bank Sta=4972,5022.8
XS Rating Curve= 0 ,0
Exp/Cntr=0.3,0.1

Type RM Length L Ch R = 1 ,51788   ,562,562,562
BEGIN DESCRIPTION:
COTTONWOOD CREEK 48.0
END DESCRIPTION:
XS GIS Cut Line= 3
      3592018.02     10656602.49      3592906.91      10656088.6
      3592934.67     10653833.42
#Sta/Elev= 30
  4137.7  318.48  4250.7  316.87  4352.7  309.13  4470.3  297.19  4535.5   294.1
  4682.4  296.28  4878.8     296  4974.2  297.98    4990  288.28  4995.8  285.73
  5002.7  285.43  5005.5  284.93  5008.7  285.43  5017.4  286.52  5027.3  294.58
  5033.1  296.96  5054.6  297.75  5172.9  294.56  5712.9  295.65    5794  294.14
  5802.9  295.65  5832.9  296.14    6533  296.22  6815.9  298.67    6883  299.47
  7018.3  313.24  7107.8  322.68    7193  331.75  7416.6  336.06  7419.8  335.09
#Mann= 7 ,-1 , 0
  4137.7     .16       0  4535.5     .12       0  5002.7     .07       0
  5008.7     .12       0  6815.9     .16       0  7018.3     .08       0
  7107.8     .12       0
Bank Sta=4974.2,5033.1
XS Rating Curve= 0 ,0
Exp/Cntr=0.3,0.1

Type RM Length L Ch R = 1 ,51226   ,195,195,195
BEGIN DESCRIPTION:
Mapping XS 86af0265
END DESCRIPTION:
XS GIS Cut Line= 3
      3592073.57     10656730.96      3593511.08     10656355.96
      3595104.75     10654866.45
#Sta/Elev= 30
  4297.8  321.71  4441.5  311.29  4603.7  295.89    4703   294.6  4893.1  293.95
  4975.8  296.95  4986.1  293.07  4997.9  285.48  5003.8  285.31  5006.5  284.81
  5009.8  285.31  5017.1  286.31  5033.2  294.98  5048.1  297.01  5161.8  297.17
  5276.1  294.67  5285.8     293  5311.4  295.04  5670.7  294.38  5917.1  294.28
  6267.6  293.79  6854.8  296.39  7165.9  309.52  7287.4  316.49  7293.8  316.47
  7538.1  331.98    7724  343.38  7817.1     348  7872.3  347.73  7964.8  343.75
#Mann= 11 ,-1 , 0
  4297.8     .16       0    4703     .12       0  5003.8     .07       0
  5009.8     .12       0  5670.7     .16       0  5917.1     .12       0
  7287.4     .16       0  7293.8     .12       0  7538.1     .16       0
    7724     .12       0  7872.3     .16       0
Bank Sta=4975.8,5048.1
XS Rating Curve= 0 ,0
Exp/Cntr=0.3,0.1

Type RM Length L Ch R = 1 ,51031   ,151,151,151
BEGIN DESCRIPTION:
COTTONWOOD CREEK 47.0
END DESCRIPTION:
XS GIS Cut Line= 4
       3592011.1     10656845.54      3592781.91     10656736.17
      3593016.29     10656694.51      3594568.35     10655949.72
#Sta/Elev= 30
    4165   321.8  4491.5     303    4592  299.53  4659.7  298.06  4893.5  295.69
  4981.8   294.5    4992  285.82  5003.7  284.87  5006.5  284.37  5009.7  284.87
  5042.8  286.71  5052.9  293.11  5198.4   293.8  5310.2  293.94  5444.7  294.27
    5508  292.05  5802.3  294.36  5869.5  294.01  5972.8   293.9  6011.8  296.28
  6221.4  306.13  6316.9  309.16  6394.3  312.76  6430.9   311.5  6540.6  312.45
  6640.4  311.74  6730.6  311.89  6764.3  314.24  6876.1  316.79  6903.1  318.04
#Mann= 20 ,-1 , 0
    4165     .08       0  4491.5     .05       0    4592     .08       0
  4659.7     .16       0  4893.5     .05       0  5003.7     .07       0
  5009.7     .08       0  5198.4     .05       0  5310.2     .16       0
  5444.7     .16       0  5802.3     .16       0  5869.5     .12       0
  6011.8     .12       0  6221.4     .16       0  6316.9     .05       0
  6430.9     .16       0  6540.6     .05       0  6640.4     .16       0
  6764.3     .05       0  6876.1     .12       0
Bank Sta=4981.8,5052.9
XS Rating Curve= 0 ,0
Exp/Cntr=0.3,0.1

Type RM Length L Ch R = 1 ,50880   ,629,629,629
BEGIN DESCRIPTION:
COTTONWOOD CREEK 46.0
END DESCRIPTION:
XS GIS Cut Line= 3
       3592276.3     10656996.18      3593489.44     10656744.43
      3594889.17     10656095.57
#Sta/Elev= 30
  4400.4   313.8    4414  311.59  4528.6  305.13  4638.7  298.76  4730.6  295.97
  4924.6   294.5  4942.2  295.64  4961.7  295.76  4975.7  295.76  4995.6   284.6
  4998.3   284.1  5001.6   284.6    5037  285.58  5043.6  289.84  5057.4  295.26
  5348.1  293.56    5590  291.74  5700.1  292.77  5789.1  293.55    6130  298.82
  6233.5  300.47  6360.7  304.07  6643.4  312.88  6682.5  314.22    6688  312.61
  6705.4  314.13  6788.9  313.68  7006.3  320.38  7065.6  320.03  7182.2  323.82
#Mann= 14 ,-1 , 0
  4400.4     .05       0  4528.6     .16       0  4942.2     .05       0
  4961.7     .16       0  4995.6     .07       0  5001.6     .16       0
  5348.1     .05       0  5700.1     .08       0  5789.1     .05       0
    6130     .08       0  6233.5     .05       0  6360.7     .08       0
  6643.4     .05       0  6788.9     .08       0
Bank Sta=4975.7,5057.4
XS Rating Curve= 0 ,0
Exp/Cntr=0.3,0.1

Type RM Length L Ch R = 1 ,50251   ,2546,2546,2546
BEGIN DESCRIPTION:
Mapping XS 68b384c8
END DESCRIPTION:
XS GIS Cut Line= 3
      3591351.34     10657543.46      3592801.01     10657491.38
      3595074.94     10656449.88
#Sta/Elev= 30
  3354.5   349.9    3673  339.86  3833.1  325.18  3865.8  325.18  4063.2  310.85
  4113.3  313.26  4173.3  311.72  4333.4  299.31  4466.8  292.85  4643.6  292.28
  4969.1  295.56  4998.5  284.69  5001.3  284.19  5004.5  284.69  5032.6  284.86
  5045.5   294.5  5055.6  294.94  5138.9  294.48  5431.2  292.14  5771.5  291.61
  6255.4  295.94    6594  305.83  6662.4  310.21  6684.4  308.99  6871.4  317.95
  6948.4  318.85  6961.1  322.11  7001.6  324.52  7024.6  323.57  7306.2  336.02
#Mann= 6 ,-1 , 0
  3354.5     .05       0  4466.8     .12       0  4998.5     .07       0
  5004.5     .12       0  5138.9     .16       0  5431.2     .05       0
Bank Sta=4969.1,5055.6
XS Rating Curve= 0 ,0
Exp/Cntr=0.3,0.1

Type RM Length L Ch R = 1 ,47705   ,1173,1173,1173
BEGIN DESCRIPTION:
COTTONWOOD CREEK 45.0
END DESCRIPTION:
XS GIS Cut Line= 4
      3590762.41     10658226.83      3592585.35     10658851.84
      3593201.67     10658591.42      3595094.03     10656916.07
#Sta/Elev= 30
  2906.7  340.39  2962.6  341.42    3168   330.4  3220.3  335.45  3268.2  337.14
  3411.2   343.5  3536.3  330.86  3662.3  325.26  4104.7  297.19    4180   295.4
    4488  290.63  4667.5  289.69  4990.4   292.9  4997.4  283.72  5000.2  283.22
  5003.4  283.72    5014  286.18    5023  291.85    5035  292.81  5232.5     291
  6359.3  290.58  6557.6  295.64  6742.2  309.96    6898  315.33  7145.6  311.59
  7379.8  317.41  7500.2  313.71  7528.7  319.74    7578  321.75  8030.3  334.74
#Mann= 13 ,-1 , 0
  2906.7     .05       0  3220.3     .16       0  3268.2     .05       0
  3536.3      .1       0  3662.3     .05       0  4104.7      .1       0
    4180     .05       0    4488     .16       0  4667.5     .05       0
  4997.4     .03       0  5003.4     .05       0    5014     .16       0
  5232.5     .05       0
Bank Sta=4990.4,5035
XS Rating Curve= 0 ,0
Exp/Cntr=0.3,0.1

Type RM Length L Ch R = 1 ,46532   ,1532,1532,1532
BEGIN DESCRIPTION:
COTTONWOOD CREEK 44.0
END DESCRIPTION:
XS GIS Cut Line= 3
      3590033.25     10659485.52      3593314.52     10659251.15
      3596056.13     10658704.56
#Sta/Elev= 30
    1591  337.79  1888.1   323.5  1918.2  315.86  1958.3  320.84  2048.5  318.66
  2155.5  307.82  2279.1  308.29  2295.8  313.97  2405.8  311.58  3333.7  294.81
  3729.9  289.98  4759.2  289.91  4962.3  292.08  5005.2  282.22  5007.9  281.72
  5011.2  282.22  5015.5  285.42  5028.6  291.48  5683.9  290.71  5706.6  286.83
  6011.6  292.16  6418.4  297.73  6537.7  306.24  6561.3  313.45  6587.5  314.69
  6754.6  314.89  6825.1  324.68  6935.4  330.53  7367.4  325.69  7676.2  332.65
#Mann= 15 ,-1 , 0
    1591     .16       0  2405.8     .05       0  3333.7      .1       0
  3729.9     .05       0  4759.2     .16       0  5005.2     .07       0
  5011.2     .16       0  5015.5     .12       0  5683.9     .16       0
  5706.6     .12       0  6011.6     .16       0  6418.4      .1       0
  6561.3     .15       0  6587.5      .1       0  6825.1     .05       0
Bank Sta=4962.3,5028.6
XS Rating Curve= 0 ,0
Exp/Cntr=0.3,0.1

Type RM Length L Ch R = 1 ,45000   ,868,868,868
BEGIN DESCRIPTION:
COTTONWOOD CREEK 43.0
END DESCRIPTION:
XS GIS Cut Line= 2
      3590546.12     10660639.32      3595884.63     10659489.15
#Sta/Elev= 30
   894.4  345.69  1409.4  314.25  1627.8  306.37  1677.1     307  1777.7  300.34
  2084.6  288.18  3738.3  288.73  4088.1  288.58  4272.4  288.78  4421.3  289.25
  4510.6   289.4  4878.1  289.62  4969.3  290.77  4979.5  283.11  4993.1  281.84
  4995.8  281.34  4999.1  281.84  5020.4  282.02  5045.4  290.65  5132.8  288.73
  5244.6  288.91    5331  289.94  5428.7  295.49  5607.1  308.83  6022.9  343.64
  6232.2  348.15  6288.9  352.22  6299.1  355.85  6325.7  359.54  6355.4  359.36
#Mann= 13 ,-1 , 0
   894.4     .05       0  3738.3     .16       0  4088.1     .05       0
  4272.4     .16       0  4421.3     .05       0  4510.6     .16       0
  4878.1     .12       0  4993.1     .07       0  4999.1     .12       0
  5132.8     .16       0  5244.6     .05       0  5428.7     .16       0
  5607.1     .05       0
Bank Sta=4969.3,5045.4
XS Rating Curve= 0 ,0
Exp/Cntr=0.3,0.1

Type RM Length L Ch R = 1 ,44132   ,537,537,537
BEGIN DESCRIPTION:
COTTONWOOD CREEK 42.0
END DESCRIPTION:
XS GIS Cut Line= 3
      3591599.64     10661460.18      3594799.61     10660460.19
      3595499.57     10660010.21
#Sta/Elev= 30
    1636  325.42  1772.2   323.1  1852.3  319.34  2257.8  291.34  2306.5  288.91
  2369.4  287.89  2474.1  288.81  2760.7  287.44  4128.9  286.46  4669.6  286.79
  4845.2  288.23  4957.1  290.29  4967.1  286.17  4972.3   285.6    4983  282.03
  4985.7  281.53    4989  282.03  5002.1  282.31  5011.4  289.79  5017.3  288.65
  5024.2  290.25  5105.1  288.15    5335  288.28    5438  296.92  5459.2  300.01
  5574.1  309.99  5610.2  314.36    5683  319.89  5725.6  324.88  5820.7  331.41
#Mann= 5 ,-1 , 0
    1636     .05       0  4845.2     .12       0    4983     .07       0
    4989     .12       0  5610.2     .16       0
Bank Sta=4957.1,5011.4
XS Rating Curve= 0 ,0
Exp/Cntr=0.3,0.1

Type RM Length L Ch R = 1 ,43595   ,549,549,549
BEGIN DESCRIPTION:
COTTONWOOD CREEK 41.0
END DESCRIPTION:
XS GIS Cut Line= 3
      3592049.65     10661660.18      3594949.61     10660960.19
       3595749.6      10660160.2
#Sta/Elev= 30
  1991.7  329.57  2156.3  315.45  2308.4  305.49  2372.3  299.17  2536.9  289.46
  2588.3  288.42  3161.5  289.62  3555.3  286.59  3716.2  288.03  3791.9   286.6
  4761.2  286.73  4863.9  288.03  4978.5  289.79  5000.2  282.52    5003  282.02
  5006.2  282.52  5017.4   283.1  5031.5  287.87  5045.7  289.31  5108.9  287.54
  5200.8  287.62  5334.3  287.69  5400.2  287.75  5467.7  287.73  5554.8  288.06
  5738.2  305.04  5823.5  312.33  5908.3  316.45  5950.8  316.55  6106.3  330.78
#Mann= 11 ,-1 , 0
  1991.7     .05       0  4761.2     .16       0  4863.9     .12       0
  5000.2     .07       0  5006.2     .12       0  5108.9     .16       0
  5200.8     .07       0  5334.3     .12       0  5400.2     .07       0
  5467.7     .12       0  5738.2     .16       0
Bank Sta=4978.5,5045.7
XS Rating Curve= 0 ,0
Exp/Cntr=0.3,0.1

Type RM Length L Ch R = 1 ,43046   ,1033,1033,1033
BEGIN DESCRIPTION:
COTTONWOOD CREEK 40.0
END DESCRIPTION:
XS GIS Cut Line= 3
      3592399.63     10661810.19      3594799.61     10661410.19
      3595899.59     10661310.19
#Sta/Elev= 30
  2568.9  317.62  2619.6  311.76  2710.8  305.66  2741.2  301.14  2913.6  291.68
  3088.5  289.37  3258.3  290.89  4144.2  286.61  4180.3  286.54  4749.8   286.7
  4951.3  289.13  4961.4   287.8    4969  280.85  4974.1  282.76  4996.5  280.26
  4999.2  279.76  5002.5  280.26  5022.1  287.79  5032.1  288.75  5062.2  289.05
  5072.3  286.58  5092.4  288.64  5102.4  287.07  5326.8  287.79  5625.9  286.88
    5735  286.88  5813.1  295.26  5821.5  295.94  5855.5  300.77  6106.5  322.42
#Mann= 10 ,-1 , 0
  2568.9     .05       0  4144.2     .16       0  4180.3     .05       0
  4749.8     .12       0  4996.5     .07       0  5002.5     .12       0
  5326.8     .07       0  5625.9     .12       0  5813.1     .16       0
  5821.5     .12       0
Bank Sta=4951.3,5032.1
XS Rating Curve= 0 ,0
Exp/Cntr=0.3,0.1

Type RM Length L Ch R = 1 ,42013   ,629,629,629
BEGIN DESCRIPTION:
COTTONWOOD CREEK 39.0
END DESCRIPTION:
XS GIS Cut Line= 4
      3592201.89     10661882.11       3594618.6     10662319.61
      3594951.93     10662236.28      3595950.96     10661334.38
#Sta/Elev= 30
  2322.1  332.11  2454.3  327.34  2685.6  306.56  2858.4  297.71    3180  291.05
  3713.3  289.15  4201.9  287.65  4251.5  285.86  4311.6  288.27  4342.1   283.5
  4358.8  287.29  4372.6  282.21  4403.1  287.29  4529.4  287.22  4582.9  281.64
  4636.4  286.59    4975  288.87  5001.6   279.2  5013.2   279.1    5016   278.6
  5019.2   279.1  5026.5   285.3  5042.9  287.98  5372.4  287.03    5740  302.52
  5769.8  302.22    5903  298.91  6037.5  301.15  6370.8  322.69  6467.6  322.22
#Mann= 8 ,-1 , 0
  2322.1     .05       0  3713.3     .16       0  4201.9     .05       0
  4251.5     .12       0  5013.2     .07       0  5019.2     .12       0
    5740     .16       0  5769.8     .12       0
Bank Sta=4975,5042.9
XS Rating Curve= 0 ,0
Exp/Cntr=0.3,0.1

Type RM Length L Ch R = 1 ,41384   ,628,628,628
BEGIN DESCRIPTION:
COTTONWOOD CREEK 38.0
END DESCRIPTION:
XS GIS Cut Line= 3
      3593340.81     10663562.68      3594875.54     10662507.11
      3596665.88     10661736.85
#Sta/Elev= 30
  3505.9  319.88  3765.8  300.29  3843.1   297.6  4190.4  286.97  4679.2  287.44
  4742.6  287.25  4751.4  283.65  4757.5  286.57  4766.3  284.06  4787.3  287.49
    4859  284.61  4966.5  287.72    4973  286.97  4984.5  278.78  4987.2  278.28
  4990.5  278.78  5002.4  278.88  5017.3  287.95  5593.4  286.68  5774.7  287.53
  6031.5  292.43  6243.9  290.49  6344.7  297.07  6446.3  300.48    6655  310.56
  6839.1  319.29  6984.4  321.42  7127.7   324.4  7237.3  324.35  7317.6  326.11
#Mann= 14 ,-1 , 0
  3505.9     .05       0  3843.1     .16       0  4190.4     .05       0
  4679.2     .12       0  4984.5     .07       0  4990.5     .12       0
  5593.4     .16       0  5774.7     .12       0  6344.7     .16       0
  6446.3     .12       0    6655     .16       0  6984.4     .05       0
  7127.7     .16       0  7237.3     .12       0
Bank Sta=4966.5,5017.3
XS Rating Curve= 0 ,0
Exp/Cntr=0.3,0.1

Type RM Length L Ch R = 1 ,40756   ,891,891,891
BEGIN DESCRIPTION:
COTTONWOOD CREEK 37.0
END DESCRIPTION:
XS GIS Cut Line= 3
      3593849.64     10664460.15      3594999.61     10662910.19
       3596399.6     10662060.19
#Sta/Elev= 30
  3031.1  329.17  3377.2   308.1  3516.7  300.38  3875.1   292.7  4002.3  285.73
  4124.5  284.38  4413.7  284.84  4552.9  283.78  4582.4   285.9  4603.2  284.24
  4961.1  287.05  4968.8  283.52  4971.7  278.52  4974.4  278.02  4977.7  278.52
  5005.6  278.57  5019.6  286.85  5353.7  286.08  5630.1   289.1  5682.1  290.25
  5724.8  295.67  5920.6  294.87    5967  306.46  6020.8  308.09  6242.3  320.07
  6287.1  319.38  6379.9  319.88  6438.1  323.72  6490.4  331.81  6598.9  336.57
#Mann= 11 ,-1 , 0
  3031.1     .05       0  3377.2     .16       0  4124.5     .05       0
  4413.7     .16       0  4552.9     .12       0  4971.7     .07       0
  4977.7     .12       0  5353.7     .16       0  5630.1     .05       0
  6020.8     .16       0  6287.1     .05       0
Bank Sta=4961.1,5019.6
XS Rating Curve= 0 ,0
Exp/Cntr=0.3,0.1

Type RM Length L Ch R = 1 ,39865   ,778,778,778
BEGIN DESCRIPTION:
COTTONWOOD CREEK 36.0
END DESCRIPTION:
XS GIS Cut Line= 2
      3594398.95      10664554.1      3596412.29     10662384.56
#Sta/Elev= 30
  3328.2   322.2  3412.9  314.65    3519  307.69    3593  298.77  3682.9  295.08
  3727.9  295.06  3833.9   283.8  3942.4   282.1  4433.8  282.94  4552.4  283.49
  4972.9  286.84  4980.2  285.46  4994.4  278.11  5005.6  278.08  5008.3  277.58
  5011.6  278.08  5022.8  286.61  5114.6  284.66  5624.3  284.38  5724.5  287.13
  5767.5  290.13  5815.3  295.14  5850.5  295.03  5919.4  300.05  5982.7  305.88
  6071.3  313.44  6111.8  316.54  6154.9     321  6271.3  328.28    6288  329.28
#Mann= 16 ,-1 , 0
  3328.2     .05       0  3412.9     .12       0    3519     .05       0
  3682.9     .16       0  3942.4     .05       0  4433.8     .16       0
  4552.4     .12       0  5005.6     .07       0  5011.6     .12       0
  5724.5     .16       0  5767.5     .05       0  5919.4     .12       0
  5982.7     .05       0  6071.3     .16       0  6111.8     .05       0
  6271.3     .12       0
Bank Sta=4972.9,5022.8
XS Rating Curve= 0 ,0
Exp/Cntr=0.3,0.1

Type RM Length L Ch R = 1 ,39087   ,1563,1563,1563
BEGIN DESCRIPTION:
COTTONWOOD CREEK 34.0
END DESCRIPTION:
XS GIS Cut Line= 2
      3594437.06     10665204.58      3597643.56     10662324.27
#Sta/Elev= 30
  3088.7  329.11  3114.6  328.62  3146.2  329.73  3256.3  329.29  3362.4  322.76
  3819.8  284.22  3833.6  283.08  3991.3  280.52  4442.2  282.31    4977  285.82
  4991.2  277.63  5002.4  277.38  5005.2  276.88  5008.4  277.38  5033.8   286.1
  5504.7  283.56  5627.8  283.56  5645.3  283.56  5765.7  283.56  5911.1  287.47
  5926.5  288.68  6041.4  302.32  6059.8  304.28  6159.6  319.47  6216.4  322.58
  6369.7  314.05  6417.9  312.14  6584.9  310.01  7044.6  320.21  7398.9  354.29
#Mann= 19 ,-1 , 0
  3088.7     .05       0  3114.6     .16       0  3146.2     .05       0
  3819.8     .16       0  3833.6     .12       0  3991.3     .05       0
  4442.2     .12       0  5002.4     .07       0  5008.4     .12       0
  5504.7     .07       0  5627.8      .1       0  5645.3     .12       0
  5765.7      .1       0  5911.1     .16       0  5926.5     .12       0
  6041.4     .16       0  6059.8     .12       0  6369.7     .16       0
  6417.9     .12       0
Bank Sta=4977,5033.8
XS Rating Curve= 0 ,0
Exp/Cntr=0.3,0.1

Type RM Length L Ch R = 1 ,37524   ,802,802,802
BEGIN DESCRIPTION:
COTTONWOOD CREEK 32.0
END DESCRIPTION:
XS GIS Cut Line= 2
      3594971.79     10665753.18      3597853.72     10663565.69
#Sta/Elev= 30
  3693.6  328.47    3829  324.95  3907.9  316.77  3986.9  314.62  4243.4  293.19
  4291.9  288.77  4393.9  282.34  4407.1   278.6  4415.4  278.76  4421.7  282.76
  4450.8  278.85  4471.6  283.22  4714.9  281.33  4958.2   284.1  4996.9  275.27
  4999.6  274.77  5002.9  275.27  5014.4  275.62  5021.6  281.48  5035.2  284.54
  5235.1  281.06  5428.3  283.86  5750.5  281.79  5783.7  281.63  5988.8  281.11
  5996.8  281.09  6499.4  280.13  6605.4  282.28  6964.8  319.13  7311.7  343.04
#Mann= 11 ,-1 , 0
  3693.6     .05       0  4243.4     .16       0  4291.9     .12       0
  4996.9     .07       0  5002.9     .12       0  5750.5     .16       0
  5783.7     .12       0  5988.8     .16       0  5996.8     .12       0
  6605.4     .16       0  6964.8     .12       0
Bank Sta=4958.2,5035.2
XS Rating Curve= 0 ,0
Exp/Cntr=0.3,0.1

Type RM Length L Ch R = 1 ,36722   ,1171,1171,1171
BEGIN DESCRIPTION:
COTTONWOOD CREEK 30.0
END DESCRIPTION:
XS GIS Cut Line= 3
      3595549.62     10665910.18      3596349.61     10665510.19
      3597899.62     10663910.18
#Sta/Elev= 30
  4108.5  322.19    4279  309.61    4367  300.13  4519.4  288.28  4533.3  285.14
  4578.1  281.54  4608.8  283.27  4667.5  281.73  4689.9  283.81  4815.6  280.74
  4966.6  284.07  4980.6  275.17  4991.5  274.66  4994.3  274.16  4997.5  274.66
  5006.4  276.12    5010   280.7    5017  283.66  5271.6  281.17  5356.5  282.33
  5731.1   280.4  5838.6  279.89  6445.6  280.08    6543   283.9  6685.9  288.97
  6792.1  295.17  6947.7  312.61  7053.7  328.27  7209.4  340.59  7230.6  340.78
#Mann= 8 ,-1 , 0
  4108.5     .05       0    4367     .12       0  4991.5     .07       0
  4997.5     .12       0  5731.1     .16       0  5838.6     .12       0
    6543     .16       0  6685.9     .12       0
Bank Sta=4966.6,5017
XS Rating Curve= 0 ,0
Exp/Cntr=0.3,0.1

Type RM Length L Ch R = 1 ,35551   ,572,572,572
BEGIN DESCRIPTION:
COTTONWOOD CREEK 28.0
END DESCRIPTION:
XS GIS Cut Line= 3
      3595949.64     10666560.17      3596749.61     10666160.19
      3598149.59     10664560.21
#Sta/Elev= 30
  4076.9  313.26  4389.9  289.55    4543   284.1  4627.5  285.85    4703  282.97
  4733.7   279.3  4839.8  282.11  4897.4  282.58  4968.5  283.07  4974.6  283.07
  4978.4  275.71  4989.6  273.96  4992.4  273.46  4995.6  273.96  5004.5  276.25
  5013.5  282.19  5021.1  283.15  5377.5  279.79  5835.5  278.21  6062.8   280.2
  6190.4  281.52  6339.5   286.9  6360.3  285.19  6466.6  287.52  6480.9  285.24
  6502.4  287.95  6588.3  296.77  6750.4  314.15  6877.6  314.87  7097.3  326.06
#Mann= 10 ,-1 , 0
  4076.9     .05       0    4543     .12       0  4839.8     .05       0
  4897.4     .12       0  4989.6     .07       0  4995.6     .12       0
  5377.5     .05       0  6062.8     .12       0  6502.4     .16       0
  6588.3     .12       0
Bank Sta=4968.5,5021.1
XS Rating Curve= 0 ,0
Exp/Cntr=0.3,0.1

Type RM Length L Ch R = 1 ,34979   ,475,475,475
BEGIN DESCRIPTION:
COTTONWOOD CREEK 27.0
END DESCRIPTION:
XS GIS Cut Line= 3
       3595860.7     10667343.44      3597360.69     10666197.61
      3598956.29     10666169.86
#Sta/Elev= 30
  3330.2  325.17  3616.8  312.49  3958.8   291.3    4109  284.42  4190.7  283.81
  4280.8  279.95  4316.2  281.59  4359.8  279.24  4373.3  281.73  4554.9  279.48
  4849.5  280.99  4972.8  283.17  4993.7  278.86  5005.2  273.67  5007.9  273.17
  5011.2  273.67  5015.1  281.31    5029  283.08  5193.2  279.42  5406.7  281.58
  5416.7  279.54  5436.7  281.45  5496.7     280    5932  321.31  6076.8  329.68
  6256.8  337.11  6336.8  337.49  6516.9  332.78  6750.5  344.36  6813.6  344.24
#Mann= 8 ,-1 , 0
  3330.2     .12       0  3616.8     .16       0  4190.7     .12       0
  4554.9     .05       0  4849.5     .12       0  5005.2     .07       0
  5011.2     .12       0  6750.5     .16       0
Bank Sta=4972.8,5029
XS Rating Curve= 0 ,0
Exp/Cntr=0.3,0.1

Type RM Length L Ch R = 1 ,34504   ,549,549,549
BEGIN DESCRIPTION:
COTTONWOOD CREEK 26.0
END DESCRIPTION:
XS GIS Cut Line= 3
      3596449.59      10667610.2      3597599.61     10666510.19
       3598099.6     10666510.19
#Sta/Elev= 30
  3407.6  324.41  3478.2  321.72  3536.1  317.71  3584.5  315.19  3662.2   308.7
    3694  304.03  3761.3  295.84  3860.3  287.83    3938  279.56  3994.5  279.21
  4077.2  279.32  4553.5  279.33  4796.2  281.35  4878.7  281.72  4885.9  280.96
  4921.2  282.19    4985  282.36  4995.5  273.11    5006  272.92  5008.8  272.42
    5012  272.92    5019  273.34    5039  281.56    5079  284.06    5089  285.98
  5227.2   300.3  5288.1  306.84    5429  324.14  5486.9  334.71    5499  336.35
#Mann= 11 ,-1 , 0
  3407.6     .12       0  3536.1     .16       0    3694     .12       0
  3994.5     .07       0  4077.2     .05       0  4796.2     .12       0
    5006     .07       0    5012     .12       0  5227.2     .16       0
  5288.1     .12       0  5486.9     .05       0
Bank Sta=4985,5039
XS Rating Curve= 0 ,0
Exp/Cntr=0.3,0.1

Type RM Length L Ch R = 1 ,33955   ,547,547,547
BEGIN DESCRIPTION:
COTTONWOOD CREEK 25.0
END DESCRIPTION:
XS GIS Cut Line= 3
      3596749.58     10667510.21      3597549.61     10667010.19
      3598149.65     10666660.17
#Sta/Elev= 30
  4067.2  304.75  4211.7  289.47  4220.5  289.72    4306  279.62    4442  279.54
  4559.2  279.26  4862.1  280.23  4966.4  281.92  4975.3  280.66  4981.7  274.95
  4987.6  275.79  4994.1  273.52  4996.8  273.02  5000.1  273.52  5013.5  275.21
  5018.5  282.14  5068.5  281.56  5077.2  282.76  5098.7  281.27  5126.4  282.18
  5200.4  280.79  5221.9  282.18  5485.3  310.12  5508.4  314.03  5515.5  316.53
  5566.3  323.09  5660.2  334.48  5670.1  334.27  5691.6  337.73  5705.3   338.4
#Mann= 6 ,-1 , 0
  4067.2     .12       0    4442     .16       0  4559.2     .05       0
  4862.1     .12       0  4994.1     .07       0  5000.1     .12       0
Bank Sta=4966.4,5018.5
XS Rating Curve= 0 ,0
Exp/Cntr=0.3,0.1

Type RM Length L Ch R = 1 ,33408   ,694,694,694
BEGIN DESCRIPTION:
COTTONWOOD CREEK 24.0
END DESCRIPTION:
XS GIS Cut Line= 3
      3596649.57     10667560.19      3597449.61     10667460.19
      3598249.61     10667060.19
#Sta/Elev= 30
    4198   317.4  4228.3  315.29  4329.1  303.91  4379.4  300.05  4477.7  287.32
  4558.3  279.41  4903.5  279.46  4953.9  281.33  4961.4  278.91  4966.5  280.93
  4981.1  272.61  4983.9  272.11  4987.1  272.61  4994.2  272.72  5001.7  277.82
  5007.1  277.82  5012.7  279.86  5018.2  275.22  5026.6  280.87    5035  281.38
  5107.7  280.92  5169.2  278.31  5191.5  278.51  5303.3  282.09    5622  286.81
  5638.8     289  5719.8  293.93  5742.2  296.82    5854  304.59  5898.7     309
#Mann= 3 ,-1 , 0
    4198     .12       0  4981.1     .07       0  4987.1     .12       0
Bank Sta=4966.5,5012.7
XS Rating Curve= 0 ,0
Exp/Cntr=0.3,0.1
