--- SALT CREEK 1.prj (project) ---

Proj Title=SALT CREEK 1 Base Level Engineering
Current Plan=p01
Default Exp/Contr=0.3,0.1
English Units
Geom File=g01
Flow File=f01
Flow File=f02
Plan File=p01
Plan File=p02
Y Axis Title=Elevation
X Axis Title(PF)=Main Channel Distance
X Axis Title(XS)=Station
BEGIN DESCRIPTION:
SALT CREEK 1
END DESCRIPTION:
DSS Export Rating Curves= 0
DSS Export Rating Curve Sorted= 0
DSS Export Volume Flow Curves= 0
DXF OffsetX= 0
DXF OffsetY= 0
DXF ScaleX= 1
DXF ScaleY= 10

--- SALT CREEK 1.p01 (plan) ---

Plan Title=Multiple Run
Short Identifier=Multiple
Geom File=g01
Flow File=f01
Subcritical Flow
K Sum by GR= 0
Std Step Tol= 0.01
Critical Tol= 0.01
Num of Std Step Trials= 20
Max Error Tol= 0.3
Flow Tol Ratio= 0.001
Split Flow NTrial= 30
Split Flow Tol= 0.02
Split Flow Ratio= 0.02
Log Output Level= 0
Friction Slope Method= 1
Unsteady Friction Slope Method= 2
Unsteady Bridges Friction Slope Method= 1
Parabolic Critical Depth
Global Vel Dist=  1 , 1 , 1
Global Log Level= 0
CheckData=True
Encroach Param= -1, 0, 0, 0
BEGIN DESCRIPTION:
Multiple Run
END DESCRIPTION:

--- SALT CREEK 1.p02 (plan) ---

Plan Title=OLD MULTI
Program Version=4.10
Short Identifier=old
Geom File=g01
Flow File=f02
Subcritical Flow
K Sum by GR= 0
Std Step Tol= 0.01
Critical Tol= 0.01
Num of Std Step Trials= 20
Max Error Tol= 0.3
Flow Tol Ratio= 0.001
Split Flow NTrial= 30
Split Flow Tol= 0.02
Split Flow Ratio= 0.02
Log Output Level= 0
Friction Slope Method= 1
Unsteady Friction Slope Method= 2
Unsteady Bridges Friction Slope Method= 1
Parabolic Critical Depth
Global Vel Dist= 1 , 1 , 1
Global Log Level= 0
CheckData=True
Encroach Param=-1 ,0,0, 0
BEGIN DESCRIPTION:
Multiple Run
END DESCRIPTION:
Computation Interval=1HOUR
Output Interval=1HOUR
Run HTab= 0
Run UNet= 0
Run PostProcess= 0
Run WQNet= 0
UNET Theta= 1
UNET Theta Warmup= 1
UNET ZTol= 0.02
UNET ZSATol= 0.05
UNET MxIter= 20
UNET MaxInSteps= 0
UNET DtIC= 0
UNET DtMin= 0
UNET MaxCRTS= 20
UNET WFStab= 2
UNET SFStab= 1
UNET WFX= 1
UNET SFX= 1
UNET DSS MLevel= 4
UNET DZMax Abort= 100
UNET Convert EG Bridges= 0
UNET Use Existing IB Tables=-1
UNET Froude Reduction=False
UNET Froude Limit= 1
UNET Froude Power= 10
UNET Time Slicing=0,0, 5
UNET Junction Losses=0
Instantaneous Interval=1HOUR
Write IC File= 0
Write IC File at Sim End=0
Echo Input=False
Echo Parameters=False
Echo Output=False
Write Detailed= 0
WQ AD Non Conservative
WQ ULTIMATE=-1
WQ Max Comp Step=1HOUR
WQ Output Interval=15MIN
WQ Output Selected Increments= 0
WQ Output face flow=0
WQ Output face velocity=0
WQ Output face area=0
WQ Output face dispersion=0
WQ Output cell volume=0
WQ Output cell surface area=0
WQ Output cell continuity=0
WQ Output cumulative cell continuity=0
WQ Output face conc=0
WQ Output face dconc_dx=0
WQ Output face courant=0
WQ Output face peclet=0
WQ Output face adv mass=0
WQ Output face disp mass=0
WQ Output cell mass=0
WQ Output cell source sink temp=0
WQ Output cell source sink nsm=0
WQ Output MaxMinRange=-1
WQ Daily Max Min Mean=-1
WQ Daily Range=0
WQ Daily Time=0
WQ Create Restart=0
WQ Fixed Restart=0
WQ System Summary=0
WQ Use Fixed Temperature=0
Sorting and Armoring Iterations= 10
XS Update Threshold= 0.02
Hydraulics Update Threshold= 0.02
Energy Slope Method= 1
Volume Change Method= 0
XS Weighting Method= 0
Number of US Weighted Cross Sections= 1
Number of DS Weighted Cross Sections= 1
Upstream XS Weight=0.25
Main XS Weight=0.5
Downstream XS Weight=0.25
Number of DS XS's Weighted with US Boundary= 1
Upstream Boundary Weight= 1
Weight of XSs Associated with US Boundary= 0
Number of US XS's Weighted with DS Boundary= 1
Downstream Boundary Weight= 0.5
Weight of XSs Associated with DS Boundary= 0.5
Sediment Output Level= 4
Mass or Volume Output= 0
Output Increment Type= 1
Profile and TS Output Increment= 10
XS Output Flag= 0
XS Output Increment= 10
Disregard all LS=0
Disregard all Conn=0
Disregard all Breaches=0
Disregard all Pumps=0

--- SALT CREEK 1.f01 (steady flow) ---

Flow Title=Multiple
Program Version=4.10
Number of Profiles= 7
Profile Names=10-year,25-year,50-year,1pct_min,100-year,1pct_plu,500-year
River Rch & RM=SALT CREEK 1,Reach-1         ,35152
    1339    1834    2239    1994    2697    3647    3900
River Rch & RM=SALT CREEK 1,Reach-1         ,27164
    2723    3851    4804    4358    5893    7970    8852
River Rch & RM=SALT CREEK 1,Reach-1         ,26800
    2723    3851    4804    4358    5893    7970    8852
River Rch & RM=SALT CREEK 1,Reach-1         ,15491
    3252    4625    5791    5268    7124    9634   10765
River Rch & RM=SALT CREEK 1,Reach-1         ,13352
    3252    4625    5791    5268    7124    9634   10765
River Rch & RM=SALT CREEK 1,Reach-1         ,5736
    3774    5389    6766    6167    8341   11280   12655
Boundary for River Rch & Prof#=SALT CREEK 1,Reach-1         , 1
Up Type= 0
Dn Type= 3
Dn Slope=0.005
Boundary for River Rch & Prof#=SALT CREEK 1,Reach-1         , 2
Up Type= 0
Dn Type= 3
Dn Slope=0.005
Boundary for River Rch & Prof#=SALT CREEK 1,Reach-1         , 3
Up Type= 0
Dn Type= 3
Dn Slope=0.005
Boundary for River Rch & Prof#=SALT CREEK 1,Reach-1         , 4
Up Type= 0
Dn Type= 3
Dn Slope=0.005
Boundary for River Rch & Prof#=SALT CREEK 1,Reach-1         , 5
Up Type= 0
Dn Type= 3
Dn Slope=0.005
Boundary for River Rch & Prof#=SALT CREEK 1,Reach-1         , 6
Up Type= 0
Dn Type= 3
Dn Slope=0.005
Boundary for River Rch & Prof#=SALT CREEK 1,Reach-1         , 7
Up Type= 0
Dn Type= 3
Dn Slope=0.005
DSS Import GetInterval= 0
DSS Import GetPeak= 0
DSS Import FillOption= 0

--- SALT CREEK 1.f02 (steady flow) ---

Flow Title=OLD Multiple
Program Version=4.10
Number of Profiles= 7
Profile Names=10-year,25-year,50-year,1pct_min,100-year,1pct_plu,500-year
River Rch & RM=SALT CREEK 1,Reach-1         ,35152
    1339    1834    2239    1994    2697    3647    3900
River Rch & RM=SALT CREEK 1,Reach-1         ,26800
    2723    3851    4804    4358    5893    7970    8852
River Rch & RM=SALT CREEK 1,Reach-1         ,13352
    3252    4625    5791    5268    7124    9634   10765
River Rch & RM=SALT CREEK 1,Reach-1         ,5736
    3774    5389    6766    6167    8341   11280   12655
Boundary for River Rch & Prof#=SALT CREEK 1,Reach-1         , 1
Up Type= 0
Dn Type= 3
Dn Slope=0.005
Boundary for River Rch & Prof#=SALT CREEK 1,Reach-1         , 2
Up Type= 0
Dn Type= 3
Dn Slope=0.005
Boundary for River Rch & Prof#=SALT CREEK 1,Reach-1         , 3
Up Type= 0
Dn Type= 3
Dn Slope=0.005
Boundary for River Rch & Prof#=SALT CREEK 1,Reach-1         , 4
Up Type= 0
Dn Type= 3
Dn Slope=0.005
Boundary for River Rch & Prof#=SALT CREEK 1,Reach-1         , 5
Up Type= 0
Dn Type= 3
Dn Slope=0.005
Boundary for River Rch & Prof#=SALT CREEK 1,Reach-1         , 6
Up Type= 0
Dn Type= 3
Dn Slope=0.005
Boundary for River Rch & Prof#=SALT CREEK 1,Reach-1         , 7
Up Type= 0
Dn Type= 3
Dn Slope=0.005
DSS Import GetInterval= 0
DSS Import GetPeak= 0
DSS Import FillOption= 0

--- SALT CREEK 1.g01 (geometry) ---

Geom Title=Existing Conditions
Program Version=4.10

River Reach=SALT CREEK 1    ,Reach-1
Reach XY= 30
      3493422.75       10600619.        3494383.       10604409.
      3495023.25       10604948.      3494769.25       10605891.
      3496224.25       10607337.      3495959.75       10607963.
       3496329.5       10608279.      3496765.75       10607988.
      3497013.25       10608893.      3497478.75       10608492.
       3498066.5       10609866.        3498460.       10609511.
      3498814.75       10609898.       3498682.5       10610276.
        3499024.       10609870.      3499871.25       10610325.
        3499913.       10610775.      3500920.25       10610530.
        3501616.       10610903.        3502355.       10610413.
       3502802.5       10609407.        3503578.       10609397.
        3504596.       10608494.      3504611.25       10607724.
      3505635.75       10607623.      3505612.75       10607206.
      3506068.75       10607298.        3506461.       10606653.
       3506584.5       10607059.       3507719.5       10606730.

Type RM Length L Ch R = 1 ,35152   ,784,784,784
BEGIN DESCRIPTION:
SALT CREEK 1 60.0
END DESCRIPTION:
XS GIS Cut Line= 3
      3492868.74      10600702.6      3493465.96     10600893.57
      3493820.13     10600803.29
#Sta/Elev= 30
  4489.6  500.15  4569.8  499.32  4672.3  497.42    4774  494.61  4791.7  492.67
  4796.9  493.37    4816  491.05  4823.8  487.92  4829.1  488.63  4847.5  487.18
  4917.3  486.67  4920.1  486.17  4923.3  486.67  4952.5  487.47  4957.7  488.28
    4963   487.2  4973.5  488.01  4995.1  487.38  5015.5  488.06  5130.7  488.05
  5161.7  491.25  5202.9  494.21    5271  497.93  5337.1  500.06    5368  503.72
  5378.4   504.2  5393.7  503.41    5399  504.73  5429.4  506.18  5482.1  507.61
#Mann= 5 ,-1 , 0
  4489.6     .05       0  4569.8     .08       0  4672.3     .05       0
  4917.3    .035       0  4923.3     .05       0
Bank Sta=4917.3,4923.3
XS Rating Curve= 0 ,0
Exp/Cntr=0.3,0.1

Type RM Length L Ch R = 1 ,34368   ,482,482,482
BEGIN DESCRIPTION:
SALT CREEK 1 59.0
END DESCRIPTION:
XS GIS Cut Line= 3
      3492849.59     10602060.21      3493449.61     10601510.19
      3493749.58     10601210.21
#Sta/Elev= 30
  4181.8  494.95  4199.9  494.89  4217.3  494.11  4241.6  493.92  4309.2   494.2
  4520.2  492.66  4535.5  493.04  4599.6  491.33    4678     491    4755  490.44
  4895.5  487.14    4911  487.04    4932  484.98    4938  484.94  4981.9  485.09
  4988.7  482.42  4989.4  481.62  4992.1  481.12  4995.4  481.62  5009.9  482.67
  5024.1   484.6  5038.2  484.87  5052.3  486.31  5066.5  486.86  5094.8  487.76
  5137.2  487.47    5321  492.37  5335.2  493.45  5349.3  493.42    5420  496.79
#Mann= 9 ,-1 , 0
  4181.8      .1       0  4199.9     .08       0  4241.6     .05       0
  4520.2      .1       0    4678     .15       0  4895.5      .1       0
    4938     .05       0  4989.4    .035       0  4995.4     .05       0
Bank Sta=4989.4,4995.4
XS Rating Curve= 0 ,0
Exp/Cntr=0.3,0.1

Type RM Length L Ch R = 1 ,33886   ,322,322,322
BEGIN DESCRIPTION:
SALT CREEK 1 58.0
END DESCRIPTION:
XS GIS Cut Line= 3
      3493399.64     10601810.18      3493649.61     10601760.19
      3493849.59      10601660.2
#Sta/Elev= 30
  4756.2  491.78  4776.6  491.56  4786.8  489.68  4854.8  488.35  4878.5  487.84
  4905.6  486.43  4929.5   484.9  4939.7  483.51  4980.5  483.12  4990.7   482.1
  4997.9  482.07  5000.7  481.57  5003.9  482.07  5008.6  482.45  5041.9  483.26
  5047.5  483.07  5064.2  483.57  5069.8  483.25  5114.5  484.02  5153.7  486.19
  5159.3  486.84  5181.6  485.61    5190  486.54  5200.5  486.99    5204  486.91
  5212.4  489.14  5220.7  491.81  5226.3  492.37  5231.9  494.21  5234.7  494.21
#Mann= 6 ,-1 , 0
  4756.2      .1       0  4854.8     .08       0  4905.6     .05       0
  4997.9    .035       0  5003.9     .05       0  5200.5     .16       0
Bank Sta=4997.9,5003.9
XS Rating Curve= 0 ,0
Exp/Cntr=0.3,0.1

Type RM Length L Ch R = 1 ,33564   ,794,794,794
BEGIN DESCRIPTION:
SALT CREEK 1 57.0
END DESCRIPTION:
XS GIS Cut Line= 2
      3493233.36     10602195.64      3494415.94     10601696.25
#Sta/Elev= 30
  4494.6  491.37  4548.7  490.88  4576.5  490.41  4831.2   488.5  4876.3  486.85
  4931.5  482.55  4989.9  481.79  4997.7  479.04  5000.5  478.54  5003.7  479.04
    5008  481.22  5031.7  482.42  5166.5  481.81  5190.2  483.87  5196.1  489.73
    5208  490.86  5219.4  491.63  5250.4  484.66  5261.2  486.21  5267.9  488.49
  5319.6  490.29  5348.8  488.33  5390.8  490.05  5402.4  491.75  5456.6  493.54
  5525.6  494.37  5559.5  493.53  5596.7  491.97  5627.2  492.36  5778.3  499.39
#Mann= 10 ,-1 , 0
  4494.6     .05       0  4548.7     .16       0  4576.5     .15       0
  4876.3     .05       0  4997.7    .035       0  5003.7     .05       0
    5208     .12       0  5267.9     .16       0  5559.5     .12       0
  5627.2     .16       0
Bank Sta=4997.7,5003.7
XS Rating Curve= 0 ,0
Exp/Cntr=0.3,0.1

Type RM Length L Ch R = 1 ,32770   ,520,520,520
BEGIN DESCRIPTION:
SALT CREEK 1 56.0
END DESCRIPTION:
XS GIS Cut Line= 3
      3493399.61     10602260.19      3493899.61     10602510.19
      3494499.62     10602460.19
#Sta/Elev= 30
  4472.7  490.29  4558.2  488.66  4666.7  486.51  4723.7   485.3  4794.1  480.91
  4861.2  482.08  4942.3  479.27  4978.6  479.79    4987  478.96  4992.4   476.6
  4995.1   476.1  4998.4   476.6  5009.4  479.72  5051.8  481.15  5086.7  479.55
    5102  480.53    5112  485.87    5122  487.61  5132.1  487.48  5162.2  481.61
  5182.2  484.36  5194.4  482.14  5209.8  478.49  5222.4  478.09  5242.4  485.22
  5266.2  485.96    5294  486.28  5393.6  488.96  5553.5  495.22  5633.8  500.95
#Mann= 11 ,-1 , 0
  4472.7     .15       0  4558.2      .1       0  4666.7     .16       0
  4723.7     .05       0  4992.4     .03       0  4998.4     .05       0
  5086.7     .12       0  5194.4     .05       0  5266.2     .16       0
    5294     .12       0  5393.6     .16       0
Bank Sta=4992.4,4998.4
XS Rating Curve= 0 ,0
Exp/Cntr=0.3,0.1

Type RM Length L Ch R = 1 ,32250   ,376,376,376
BEGIN DESCRIPTION:
SALT CREEK 1 55.0
END DESCRIPTION:
XS GIS Cut Line= 2
      3493291.91     10603005.12      3494643.52     10602617.09
#Sta/Elev= 30
  4338.1  491.02  4398.3  489.75  4502.4   489.1  4591.1  486.48  4668.9  486.36
  4928.7  482.61    4988  477.93  4998.6  474.36  5001.3  473.86  5004.6  474.36
    5012  476.88  5043.2  477.29  5065.9  480.09  5084.8  480.02  5094.4  482.85
    5116  485.57  5126.4  485.19  5129.6  483.93  5145.4  480.04  5157.6   476.5
  5172.3  476.57  5178.4  479.87    5206  480.19  5261.7  484.44  5509.1  493.55
  5562.6  497.01    5658  501.88  5688.2   502.7  5714.6  505.13  5744.3  506.26
#Mann= 10 ,-1 , 0
  4338.1      .1       0  4398.3     .08       0  4502.4     .05       0
  4998.6     .03       0  5004.6     .05       0  5129.6     .16       0
  5145.4     .12       0  5509.1     .16       0  5562.6      .1       0
    5658     .16       0
Bank Sta=4998.6,5004.6
XS Rating Curve= 0 ,0
Exp/Cntr=0.3,0.1

Type RM Length L Ch R = 1 ,31874   ,548,548,548
BEGIN DESCRIPTION:
SALT CREEK 1 54.0
END DESCRIPTION:
XS GIS Cut Line= 2
       3493304.9     10603322.84      3494719.01     10602979.07
#Sta/Elev= 30
  4244.5  491.99  4380.1  490.62  4446.7  489.05  4712.5  484.82  4823.9  484.86
  4835.9  482.94  4870.8  482.18  4907.4  478.58    4980  476.96  4998.2  471.73
  5000.9  471.23  5004.2  471.73  5010.9  476.06  5021.2  475.86  5031.5  477.96
  5037.8   481.4  5042.9  478.44  5052.1  482.68  5062.4  483.95  5084.7  481.83
  5093.2  477.45  5103.5  474.99  5113.8  476.84  5202.5  476.64  5319.6  478.62
  5360.8  481.63    5382  485.11  5427.4  487.92  5607.8  499.61  5699.8  500.89
#Mann= 7 ,-1 , 0
  4244.5     .05       0  4380.1      .1       0  4446.7     .05       0
  4998.2    .035       0  5004.2     .05       0  5202.5     .16       0
  5427.4     .05       0
Bank Sta=4998.2,5004.2
XS Rating Curve= 0 ,0
Exp/Cntr=0.3,0.1

Type RM Length L Ch R = 1 ,31326   ,601,601,601
BEGIN DESCRIPTION:
SALT CREEK 1 53.0
END DESCRIPTION:
XS GIS Cut Line= 3
      3493460.18     10603604.54      3494435.84      10603521.2
       3494938.9     10603104.88
#Sta/Elev= 30
  4179.2   489.8  4439.6  487.77  4529.9  485.85    4560  486.48  4600.2  485.65
  4630.3  487.89  4638.4  485.62  4690.5  484.54  4762.4  484.85  4770.8  483.13
    4841  480.98  4851.1     479  4861.1  478.44  4891.2  481.57  4901.2  480.67
  4911.3  477.01  4931.4  473.59  4939.9  473.62  4981.5  474.39  4992.3  471.83
  4995.1  471.33  4998.3  471.83  5011.6  475.28  5051.8  473.71  5081.9  477.37
  5183.2  480.87  5345.9  483.97  5379.2  485.53  5658.6  494.76  5811.4  502.58
#Mann= 5 ,-1 , 0
  4179.2     .05       0  4939.9     .16       0  4992.3     .07       0
  4998.3     .16       0  5379.2     .05       0
Bank Sta=4992.3,4998.3
XS Rating Curve= 0 ,0
Exp/Cntr=0.3,0.1

Type RM Length L Ch R = 1 ,30725   ,552,552,552
BEGIN DESCRIPTION:
SALT CREEK 1 52.0
END DESCRIPTION:
XS GIS Cut Line= 3
      3493549.63     10604160.19      3494349.61     10604010.19
      3494949.61     10603260.18
#Sta/Elev= 30
  4171.7  490.06  4223.3  486.55  4375.2  483.57  4527.5  484.93  4710.9  483.62
  4782.1  481.43    4833  478.03  4843.2  473.44  4883.9  479.94  4894.1  479.47
  4911.5  475.07  4924.6  472.74  4965.3  473.99  4992.8  472.28  5010.6   467.8
  5013.4   467.3  5016.6   467.8    5028  472.74  5063.3  470.45  5085.7  473.46
  5184.9  472.69  5191.3  474.18  5269.8  474.88  5305.8  480.72  5369.8  479.96
  5383.4  482.29  5426.6  481.48  5521.9  484.15  5899.1  498.94  5946.1  500.15
#Mann= 8 ,-1 , 0
  4171.7      .1       0  4223.3     .08       0  4527.5     .05       0
  4911.5     .16       0  5010.6     .07       0  5016.6     .16       0
  5521.9     .05       0  5899.1     .16       0
Bank Sta=5010.6,5016.6
XS Rating Curve= 0 ,0
Exp/Cntr=0.3,0.1

Type RM Length L Ch R = 1 ,30173   ,468,468,468
BEGIN DESCRIPTION:
SALT CREEK 1 51.0
END DESCRIPTION:
XS GIS Cut Line= 3
      3494149.59     10604410.19      3494399.61     10604410.19
      3494799.61     10604010.19
#Sta/Elev= 30
  4765.7  482.82  4775.7  482.18  4785.7  482.61  4825.7  481.68  4835.7  478.75
  4855.7  475.02  4865.7  474.41  4895.7  474.41  4905.7  475.95  4925.7  480.38
  4935.7  480.15  4955.7  473.45  4965.7  470.85  4975.7  470.23  4992.7  467.73
  4995.5  467.23  4998.7  467.73  5013.2   469.9  5019.3   469.9  5029.9  471.46
    5044  472.37  5100.6  472.34  5171.3  475.97  5227.8  475.23  5284.4  477.08
  5383.4  478.56  5397.6  479.92  5425.9  480.39  5477.8  481.19  5581.4   482.9
#Mann= 5 ,-1 , 0
  4765.7     .05       0  4992.7     .07       0  4998.7     .05       0
  5425.9      .1       0  5477.8     .16       0
Bank Sta=4992.7,4998.7
XS Rating Curve= 0 ,0
Exp/Cntr=0.3,0.1

Type RM Length L Ch R = 1 ,29705   ,488,488,488
BEGIN DESCRIPTION:
SALT CREEK 1 50.0
END DESCRIPTION:
XS GIS Cut Line= 3
      3493799.64     10604810.19      3494699.61     10604710.19
       3495099.6     10604560.19
#Sta/Elev= 30
  4087.7  486.24  4159.7  484.35  4449.9  480.48  4600.8  480.34    4631  478.96
  4661.2  480.98  4681.3  477.66  4691.4  474.27  4711.5  473.51  4761.8  476.49
    4792  474.63  4822.2  471.08  4859.5  470.14  4983.1  470.14  4990.7  467.07
    5000  466.96  5002.7  466.46    5006  466.96  5014.6  470.09  5033.3  472.36
  5046.6  472.71  5068.9   469.5  5078.6   470.5    5149  471.93  5185.4  476.88
  5204.1  478.42    5292  482.13  5380.4  486.25  5399.1   488.2  5420.4  488.55
#Mann= 6 ,-1 , 0
  4087.7      .1       0  4159.7     .05       0  4859.5     .16       0
    5000     .07       0    5006     .16       0    5292     .05       0
Bank Sta=5000,5006
XS Rating Curve= 0 ,0
Exp/Cntr=0.3,0.1

Type RM Length L Ch R = 1 ,29217   ,614,614,614
BEGIN DESCRIPTION:
SALT CREEK 1 49.0
END DESCRIPTION:
XS GIS Cut Line= 3
      3493873.52     10604982.26      3494826.23     10604934.51
      3495305.21     10604566.07
#Sta/Elev= 30
  3864.6  485.24  3870.7  484.19  3890.7  484.83  3910.7  483.76  4181.1  482.37
  4351.3  478.23  4400.9   481.1  4431.4  475.91  4441.4  475.29  4511.5  475.76
  4621.6  472.15  4672.1  473.54  4748.3  470.91  4831.4   467.9  4856.1  469.07
  4987.3  468.34  4992.5  464.65  4995.2  464.15  4998.5  464.65  5001.8  465.65
    5010  471.89  5016.3  474.42  5037.2  479.12  5045.3  478.64  5113.6  482.96
  5194.8  487.01  5259.1  491.94  5279.9  492.29    5309  495.39  5422.8  498.58
#Mann= 7 ,-1 , 0
  3864.6     .05       0  4672.1     .16       0  4748.3     .05       0
  4856.1     .16       0  4992.5     .07       0  4998.5     .16       0
  5113.6     .05       0
Bank Sta=4992.5,4998.5
XS Rating Curve= 0 ,0
Exp/Cntr=0.3,0.1

Type RM Length L Ch R = 1 ,28603   ,88,88,88
BEGIN DESCRIPTION:
SALT CREEK 1 48.0
END DESCRIPTION:
XS GIS Cut Line= 2
      3494559.49      10605670.6      3495178.49     10604814.06
#Sta/Elev= 30
  4521.9  473.42  4551.3  473.84    4559  474.78  4565.2  471.71  4571.8  475.99
  4579.9  476.19  4600.8  472.29  4786.6  469.21  4824.5  467.34  4902.5  466.54
  4908.7  469.97  4917.2  465.96  4923.4   469.4  4938.1  466.02  4944.2  469.46
  4952.8  466.87  4958.9   470.3  4979.8  464.62  5023.9  463.89  5044.8  468.52
  5056.5  463.82  5059.3  463.32  5062.5  463.82  5065.7  468.28  5201.8  470.21
  5260.6  466.18  5281.5   469.3  5287.7  472.85  5488.8  481.33  5578.7  488.27
#Mann= 6 ,-1 , 0
  4521.9     .08       0  4551.3     .05       0  4786.6      .1       0
  4824.5     .05       0  5056.5     .04       0  5062.5     .05       0
Bank Sta=5056.5,5062.5
XS Rating Curve= 0 ,0
Exp/Cntr=0.3,0.1

Type RM Length L Ch R = 1 ,28515   ,923,923,923
BEGIN DESCRIPTION:
SALT CREEK 1 47.0
END DESCRIPTION:
XS GIS Cut Line= 2
      3494595.96     10605745.24      3495269.58     10604856.34
#Sta/Elev= 30
    4490  474.54  4540.9  471.28  4567.9  470.69  4624.2  466.38  4646.9  466.26
  4653.3  468.19  4659.5  466.59  4667.8  468.17  4674.1  465.96  4682.4  466.98
  4838.4  465.96  4867.5  467.39  4902.9  466.02  4967.4  467.14  4993.5   462.4
  4996.2   461.9  4999.5   462.4  5017.3  466.95  5031.9  468.98  5131.7  469.17
  5302.3  474.79  5331.4  474.45  5337.7  475.76  5360.5  475.72  5495.8  481.94
  5502.1  483.49  5524.9  483.74  5531.2  485.44  5545.7  485.05  5605.3  489.05
#Mann= 4 ,-1 , 0
    4490     .08       0  4540.9     .05       0  4993.5     .04       0
  4999.5     .05       0
Bank Sta=4993.5,4999.5
XS Rating Curve= 0 ,0
Exp/Cntr=0.3,0.1

Type RM Length L Ch R = 1 ,27592   ,428,428,428
BEGIN DESCRIPTION:
SALT CREEK 1 46.0
END DESCRIPTION:
XS GIS Cut Line= 4
      3494410.65     10605955.84      3494803.02     10606013.13
      3494865.52     10605999.24      3495358.77     10605684.25
#Sta/Elev= 30
  4571.1  474.78  4579.3  474.81  4691.3   474.8  4705.8  473.33  4711.5  474.07
  4721.6  477.92  4731.7  479.39    4752  477.74  4762.1  473.49  4782.3  471.06
  4822.7  470.52  4832.8  469.71  4845.7  466.03  4967.6  464.92  4984.6  463.66
  4999.1  458.21  5001.9  457.71  5005.1  458.21  5007.2  458.32  5015.4  462.93
  5025.6  462.79  5040.8  464.63    5084  465.15  5273.8  465.76  5301.4  466.61
  5316.6  469.13  5337.8  469.28  5358.9  470.89  5489.2  473.12  5616.9  476.75
#Mann= 4 ,-1 , 0
  4571.1     .15       0  4579.3     .05       0  4999.1     .03       0
  5005.1     .05       0
Bank Sta=4984.6,5015.4
XS Rating Curve= 0 ,0
Exp/Cntr=0.3,0.1

Type RM Length L Ch R = 1 ,27164   ,364,364,364
BEGIN DESCRIPTION:
SALT CREEK 1 45.0
END DESCRIPTION:
XS GIS Cut Line= 3
       3494749.6      10606560.2      3495149.61     10606260.19
      3495399.59     10605910.21
#Sta/Elev= 30
    4510  473.05  4617.3  471.01  4667.3  469.04  4673.6  467.61  4702.7  465.97
  4731.9  466.26  4802.7  464.25  4867.3  465.29  4873.6  459.43  4881.9  457.18
  4888.1  460.49  4902.7  460.91    4910  459.97  4914.3  457.04  4917.1  456.54
  4920.3  457.04  4923.6  461.84  4931.9  461.82  4938.1   463.7  4973.6  463.55
  4981.9  460.96  4996.5  459.84  5002.7  457.15  5006.9  462.77  5032.1  464.25
  5067.8  463.67  5195.6  468.72  5296.3  469.61    5418  473.08  5440.1  472.75
#Mann= 3 ,-1 , 0
    4510     .05       0  4914.3     .03       0  4920.3     .05       0
Bank Sta=4914.3,4920.3
XS Rating Curve= 0 ,0
Exp/Cntr=0.3,0.1

Type RM Length L Ch R = 1 ,26800   ,497,497,497
BEGIN DESCRIPTION:
SALT CREEK 1 44.0
END DESCRIPTION:
XS GIS Cut Line= 3
      3494749.62     10607110.17      3495299.61     10606510.19
      3495699.59     10605710.23
#Sta/Elev= 30
    4250  477.94  4263.9  479.29  4279.4  478.89  4285.4  478.52  4292.2  475.68
  4320.6  473.72  4370.5  475.02  4391.5  473.62  4936.6  469.88  4979.1  465.87
  4985.9  458.91  4997.1  455.62  4999.8  455.12  5003.1  455.62  5007.5  458.18
  5021.7  459.12  5028.5  457.97  5035.9  460.12  5056.8  459.16  5060.5  461.62
  5066.7  461.62  5077.9  463.97  5100.3  463.11  5251.2  464.49  5502.7  469.09
    5690  476.12  5771.1  477.64  5832.6   480.2  5854.9  482.91  5958.3  487.41
#Mann= 4 ,-1 , 0
    4250     .08       0  4279.4     .05       0  4997.1     .03       0
  5003.1     .05       0
Bank Sta=4997.1,5003.1
XS Rating Curve= 0 ,0
Exp/Cntr=0.3,0.1

Type RM Length L Ch R = 1 ,26303   ,455,455,455
BEGIN DESCRIPTION:
SALT CREEK 1 43.0
END DESCRIPTION:
XS GIS Cut Line= 3
      3495249.62     10606960.18      3495749.61     10606610.19
      3496149.59      10606410.2
#Sta/Elev= 30
  4418.6  471.88  4440.8  471.27  4518.4  471.47  4562.9   470.2    4569  470.72
  4589.9  470.17  4619.6  470.62  4655.3  469.37  4771.3  467.33  4813.1  463.18
  4827.9  462.85  4914.3  463.57  4920.4  464.16  4943.5  461.58  4985.8  460.16
  4997.6  456.09  5000.3  455.59  5003.6  456.09  5015.4  457.22  5021.5  462.83
  5031.7  462.46  5037.3  463.36  5149.1  463.34  5244.1  466.04  5305.6  466.06
    5342  467.44  5378.3   469.9  5395.1  469.68  5467.7  472.95  5476.1  472.68
#Mann= 3 ,-1 , 0
  4418.6     .05       0  4997.6     .03       0  5003.6     .05       0
Bank Sta=4997.6,5003.6
XS Rating Curve= 0 ,0
Exp/Cntr=0.3,0.1

Type RM Length L Ch R = 1 ,25848   ,433,433,433
BEGIN DESCRIPTION:
SALT CREEK 1 42.0
END DESCRIPTION:
XS GIS Cut Line= 3
      3494799.59      10607310.2      3495899.61     10606910.19
      3496549.64     10606360.17
#Sta/Elev= 30
  3803.4  479.69  3835.3  475.07  3856.6  474.33  3874.6  475.85  3905.2  474.08
  4005.6  473.01  4122.6  473.15  4154.6  471.88  4434.5  470.48  4484.4  471.17
  4668.6  468.28  4707.9  466.26  4819.2   463.9  4897.4  462.59  4952.6   463.5
  4963.9  460.96  4977.2  460.23  4998.9  456.07  5001.6  455.57  5004.9  456.07
  5012.3  458.92  5023.9  462.47  5052.5  462.34  5065.6  459.96  5079.9  462.25
  5122.8  462.35  5208.5   466.4  5342.5  468.63  5477.6   473.5  5825.4  493.57
#Mann= 5 ,-1 , 0
  3803.4     .05       0  4819.2     .16       0  4998.9     .07       0
  5004.9     .16       0  5012.3     .05       0
Bank Sta=4998.9,5004.9
XS Rating Curve= 0 ,0
Exp/Cntr=0.3,0.1

Type RM Length L Ch R = 1 ,25415   ,570,570,570
BEGIN DESCRIPTION:
SALT CREEK 1 41.0
END DESCRIPTION:
XS GIS Cut Line= 3
      3495535.74     10607508.64      3496091.32     10607144.04
      3496555.15     10606506.81
#Sta/Elev= 30
  4448.1  470.32  4536.5  468.28    4550  468.92  4565.1  467.45  4601.2  466.88
  4616.3  465.78  4703.7  464.09  4955.1  462.59  4962.9  460.41    4984  458.31
  4999.1  455.53  5017.1  455.45  5019.9  454.95  5023.1  455.45  5035.2  461.99
  5041.2  462.38  5142.1  461.89  5150.3  462.45  5221.4  461.15  5307.1  462.59
  5357.4   462.5    5372  464.82  5378.2  462.99  5386.7   463.8  5407.6  463.76
  5436.9  467.14    5464  467.15  5550.3  472.42  5636.9  474.53  5900.8  486.38
#Mann= 3 ,-1 , 0
  4448.1     .05       0  5017.1     .03       0  5023.1     .05       0
Bank Sta=5017.1,5023.1
XS Rating Curve= 0 ,0
Exp/Cntr=0.3,0.1

Type RM Length L Ch R = 1 ,24845   ,945,945,945
BEGIN DESCRIPTION:
SALT CREEK 1 40.0
END DESCRIPTION:
XS GIS Cut Line= 3
      3495549.61     10607610.19      3496199.61     10607610.19
       3496499.6      10607360.2
#Sta/Elev= 30
  4338.2  471.09  4438.2  468.57  4448.2  469.07  4458.2  468.24  4498.2  467.56
  4578.2   463.9  4648.2  462.06  4789.4  460.99  4858.2  460.87  4868.2  460.37
  4888.2  461.32  4948.2  461.35  4958.2  460.98  4968.2  459.52  4978.2  456.72
  4982.7  454.11  4985.5  453.61  4988.7  454.11  5001.9  454.66  5009.7  455.79
  5016.2  455.48    5024  461.93  5073.5  460.81  5102.1  460.85  5122.9  461.63
  5144.4  464.29  5186.7  466.65  5229.7  466.86  5264.8  467.24  5378.7  470.32
#Mann= 5 ,-1 , 0
  4338.2     .05       0  4789.4     .16       0  4982.7     .07       0
  4988.7     .16       0  5229.7     .05       0
Bank Sta=4982.7,4988.7
XS Rating Curve= 0 ,0
Exp/Cntr=0.3,0.1

Type RM Length L Ch R = 1 ,23900   ,1793,1793,1793
BEGIN DESCRIPTION:
SALT CREEK 1 39.0
END DESCRIPTION:
XS GIS Cut Line= 3
      3495392.58     10608107.59      3496030.55     10608159.67
      3496868.21     10607187.46
#Sta/Elev= 30
    4135  473.62  4463.1  472.45  4633.7  469.26  4778.1  468.65  4873.3  464.76
  4901.8  461.24  4965.5  460.11  4986.3   455.4    4991  450.65  4993.7  450.15
    4997  450.65  5000.6  451.81  5008.3  451.63  5014.9  456.33  5022.5  459.43
  5064.8  460.34  5078.5  459.19  5154.9  461.03  5227.7  460.58  5280.1  462.63
  5382.4  464.01  5405.3  464.65  5639.1   470.4  5702.8  470.12  5710.4  471.37
  5766.4  473.39  5880.5  481.26  5986.9  487.01  6028.6  493.56  6058.4  495.09
#Mann= 7 ,-1 , 0
    4135     .05       0    4991    .035       0    4997     .05       0
  5154.9     .16       0  5280.1     .05       0  5382.4     .16       0
  5405.3     .05       0
Bank Sta=4991,4997
XS Rating Curve= 0 ,0
Exp/Cntr=0.3,0.1

Type RM Length L Ch R = 1 ,22107   ,216,216,216
BEGIN DESCRIPTION:
SALT CREEK 1 37.0
END DESCRIPTION:
XS GIS Cut Line= 3
      3496191.98     10608927.77       3496900.3     10608358.33
      3497329.53     10607873.72
#Sta/Elev= 30
  4178.2   470.3  4309.9  468.82  4330.8  470.06  4338.7  468.02  4388.3  467.37
  4423.5  469.33  4452.3  466.12  4743.5  461.11  4778.7  462.85  4829.5  462.44
  4836.3  459.83  4857.1  458.63  4957.8  458.02  4970.7  453.64  4985.1  453.49
  4996.5   449.1  4999.3   448.6  5002.5   449.1  5013.9   450.8  5021.9  457.73
  5028.3  459.03  5080.5  457.56  5368.4  457.25  5382.6  458.29  5390.1  460.64
  5396.8  459.67  5418.5  464.34    5503  468.69  5616.8  478.72  5734.4  492.98
#Mann= 4 ,-1 , 0
  4178.2     .05       0  4996.5    .035       0  5002.5     .05       0
  5080.5     .16       0
Bank Sta=4996.5,5002.5
XS Rating Curve= 0 ,0
Exp/Cntr=0.3,0.1

Type RM Length L Ch R = 1 ,21891   ,1388,1388,1388
BEGIN DESCRIPTION:
SALT CREEK 1 36.0
END DESCRIPTION:
XS GIS Cut Line= 3
      3496549.64     10608860.17      3496899.61     10608610.19
      3497249.62     10608210.18
#Sta/Elev= 30
    4577  464.71  4670.4  462.72  4857.2  461.28  4907.5  459.45  4913.7  460.03
  4928.4  459.31  4943.2  460.85  4949.3  460.66  4957.9  456.86  4996.7   450.1
  4999.5   449.6  5002.7   450.1  5010.4  450.16  5020.8  455.75  5035.1  456.65
    5092  455.86  5155.6  457.65  5169.9  457.71  5177.4  456.96  5184.1  458.21
  5191.7  457.55  5212.6  458.74  5219.7  458.54  5226.8  457.27  5233.4  458.52
    5241  458.17  5293.8  460.24    5446  464.39  5524.8  468.04  5538.6  469.68
#Mann= 4 ,-1 , 0
    4577     .05       0  4996.7    .035       0  5002.7     .05       0
  5293.8     .16       0
Bank Sta=4996.7,5002.7
XS Rating Curve= 0 ,0
Exp/Cntr=0.3,0.1

Type RM Length L Ch R = 1 ,20503   ,493,493,493
BEGIN DESCRIPTION:
SALT CREEK 1 35.0
END DESCRIPTION:
XS GIS Cut Line= 2
       3496751.9     10609565.71      3497861.28     10608435.49
#Sta/Elev= 30
  3945.3  467.95    3997   466.2  4053.6  466.51    4089  463.92  4407.2  459.34
  4449.6  457.44  4456.8  458.75  4562.8  459.08  4739.5  455.78  4817.4  456.01
  4838.5   452.9    4973  454.91  4998.3  447.24    5001  446.74  5004.3  447.24
  5008.3  450.06  5029.5  451.73  5036.6  453.93  5043.7  452.09  5050.7  453.25
  5057.8  451.85  5064.8  455.54    5072  453.81  5086.1  453.96  5093.1  457.48
  5114.4  457.28  5142.7  460.02  5156.8  462.94  5227.6  465.38    5529  485.09
#Mann= 3 ,-1 , 0
  3945.3     .05       0  4998.3    .035       0  5004.3     .05       0
Bank Sta=4998.3,5004.3
XS Rating Curve= 0 ,0
Exp/Cntr=0.3,0.1

Type RM Length L Ch R = 1 ,20010   ,688,688,688
BEGIN DESCRIPTION:
SALT CREEK 1 34.0
END DESCRIPTION:
XS GIS Cut Line= 3
       3497049.6      10609710.2      3497799.61     10609010.19
      3498099.59     10608610.21
#Sta/Elev= 30
  3954.8   463.9    4428  458.57  4520.8   457.4  4534.9  453.24  4542.3  455.18
  4591.6  451.37  4761.6  454.61  4803.6  453.02  4887.7   454.2  4952.6  452.28
  4973.6  448.07  4983.9  449.36    4988  446.65  4994.3  447.35  5005.9  445.23
  5008.6  444.73  5011.9  445.23  5017.2  453.79  5044.3  462.63  5152.6  463.31
  5194.3  459.83  5202.6  461.77  5208.9  459.33  5223.4  459.43  5252.6  465.07
  5358.9  463.63  5408.9  474.17  5452.6  487.08  5467.2  486.54  5480.7  482.74
#Mann= 5 ,-1 , 0
  3954.8     .05       0    4428     .16       0  4887.7     .05       0
  5005.9    .035       0  5011.9     .05       0
Bank Sta=5005.9,5011.9
XS Rating Curve= 0 ,0
Exp/Cntr=0.3,0.1

Type RM Length L Ch R = 1 ,19322   ,512,512,512
BEGIN DESCRIPTION:
SALT CREEK 1 33.0
END DESCRIPTION:
XS GIS Cut Line= 3
      3497387.32     10609841.74      3497863.89     10609331.32
      3498193.79     10609084.55
#Sta/Elev= 30
  4243.9  461.97  4423.7  458.87  4536.6  459.69  4543.9  457.15  4600.6  456.11
  4628.9  452.68  4819.9  454.85  4840.9  454.54  4861.9  451.11  4942.2  452.82
    4954  450.45  4974.9  450.51  4986.5  443.52  4989.2  443.02  4992.5  443.52
  5011.8  444.66  5018.6  453.67  5039.5  455.05  5104.1  451.56  5118.7  453.16
  5133.3  451.67  5139.5  448.31  5154.1     449  5161.7  452.69  5174.9  452.69
  5189.5  455.83  5233.3  459.84  5304.2  463.08    5325  466.12  5354.2  473.59
#Mann= 3 ,-1 , 0
  4243.9     .05       0  4986.5    .035       0  4992.5     .05       0
Bank Sta=4986.5,4992.5
XS Rating Curve= 0 ,0
Exp/Cntr=0.3,0.1

Type RM Length L Ch R = 1 ,18810   ,1005,1005,1005
BEGIN DESCRIPTION:
SALT CREEK 1 32.0
END DESCRIPTION:
XS GIS Cut Line= 3
      3497799.58     10609860.21      3498049.61     10609610.19
      3498249.61     10609210.19
#Sta/Elev= 30
  4648.5  458.94  4846.5  457.22  4860.7  455.81  4917.2  453.95  4931.4  452.71
  4945.5  447.22  4959.7  446.75  4973.8  443.95  4995.6  442.29  4998.3  441.79
  5001.6  442.29  5010.5  442.48  5016.1  444.33  5024.5  444.57  5032.8  451.01
  5038.4  449.98  5055.2  451.43  5077.6  451.43  5083.1  448.71  5099.9  448.42
  5113.9  450.41  5127.9  454.29  5150.2  454.15    5167  453.04    5181  454.06
  5211.7  453.86  5225.7  455.23  5284.4   455.9  5329.1  457.46  5449.3  463.73
#Mann= 3 ,-1 , 0
  4648.5     .05       0  4995.6    .035       0  5001.6     .05       0
Bank Sta=4995.6,5001.6
XS Rating Curve= 0 ,0
Exp/Cntr=0.3,0.1

Type RM Length L Ch R = 1 ,17805   ,1104,1104,1104
BEGIN DESCRIPTION:
SALT CREEK 1 31.0
END DESCRIPTION:
XS GIS Cut Line= 3
      3498124.76     10610080.51      3498499.61     10609560.19
      3498849.61     10609310.19
#Sta/Elev= 30
  4323.7  458.69  4542.8  454.34  4643.4   454.2    4679  452.23  4693.7  453.43
  4714.6  451.51  4764.9   453.9  4968.1  450.08  4987.1  447.63  4993.2  445.63
  4998.8  441.53  5001.6  441.03  5004.8  441.53  5014.1   443.2  5022.7  447.73
  5028.9   453.7  5037.5  453.04  5043.6  455.27    5051  451.67  5058.4  456.88
    5137  462.11  5150.5  462.12  5159.1  459.61  5186.2  461.41  5194.8  459.07
  5200.9  460.22  5209.5  457.34  5230.4  461.92  5301.7  464.74  5395.1  475.23
#Mann= 3 ,-1 , 0
  4323.7     .05       0  4998.8    .035       0  5004.8     .05       0
Bank Sta=4968.1,5028.9
XS Rating Curve= 0 ,0
Exp/Cntr=0.3,0.1

Type RM Length L Ch R = 1 ,16701   ,1210,1210,1210
BEGIN DESCRIPTION:
Mapping XS 846bd60a
END DESCRIPTION:
XS GIS Cut Line= 3
      3498286.46     10610326.18      3498889.75     10610015.86
      3499080.67     10609365.01
#Sta/Elev= 30
  4609.8  459.49  4892.5  455.14  4973.2   451.6  4981.2  440.68  4986.8  442.28
  4995.7  439.99  5003.4   441.1    5006  439.77  5008.8  439.27    5012  439.77
  5025.6  445.33  5053.4  445.61  5063.2  446.58  5069.9  449.57  5108.1  449.09
  5247.3  451.89    5315   448.6  5387.9  447.57  5407.8  449.68  5451.6   449.7
  5471.3  451.03  5479.8   453.5  5492.1  453.75  5502.6  453.42  5518.4   450.4
  5523.6  455.45  5533.8  456.19  5648.5  461.43  5695.8  465.17  5966.5  477.26
#Mann= 3 ,-1 , 0
  4609.8     .05       0    5006    .035       0    5012     .05       0
Bank Sta=4973.2,5069.9
XS Rating Curve= 0 ,0
Exp/Cntr=0.3,0.1

Type RM Length L Ch R = 1 ,15491   ,484,484,484
BEGIN DESCRIPTION:
SALT CREEK 1 30.0
END DESCRIPTION:
XS GIS Cut Line= 2
      3498759.99      10611327.9      3499447.49     10609550.11
#Sta/Elev= 30
  3641.3  460.02  3788.2   458.9  3818.1  454.55  3842.6  458.32    4132  453.47
  4210.5  447.55  4217.8  450.91  4239.9  450.18  4287.1  451.31    4295  447.74
  4314.2  449.91  4319.6  447.66  4357.2  452.61  4700.3  451.56  4875.6  448.12
  4895.2  450.56  4960.1  450.96  4979.1  445.54  4984.7  436.91    4990  439.19
  4997.5  436.79  5000.3  436.29  5003.5  436.79    5022  443.67  5069.1  451.23
  5127.3  462.83  5208.1  474.67  5292.6  482.22  5431.6  492.61  5547.4  497.51
#Mann= 7 ,-1 , 0
  3641.3     .05       0  4239.9      .1       0  4287.1     .05       0
  4895.2      .1       0  4997.5     .07       0  5003.5      .1       0
  5127.3     .05       0
Bank Sta=4960.1,5069.1
XS Rating Curve= 0 ,0
Exp/Cntr=0.3,0.1

Type RM Length L Ch R = 1 ,15007   ,551,551,551
BEGIN DESCRIPTION:
SALT CREEK 1 27.0
END DESCRIPTION:
XS GIS Cut Line= 2
      3499159.28     10611282.79      3499631.51     10609758.46
#Sta/Elev= 30
  3904.9  457.25  3993.5  459.24  4012.3  456.13  4085.6  453.01  4106.5  449.78
  4123.9  452.56  4148.4  452.62    4226  447.11  4284.5   451.1  4315.9  448.19
  4372.9  448.19    4433  447.86  4472.9  451.22  4514.8  451.29    4772  447.47
  4912.6  449.83  4975.6   447.7  4985.9  438.94  5005.2  435.86  5007.9  435.36
  5011.2  435.86  5017.3   440.2  5048.7   444.3  5059.2  448.56    5077  451.85
  5184.3  465.11  5306.8  478.63    5372  483.36  5409.8  482.92  5500.7  490.59
#Mann= 8 ,-1 , 0
  3904.9     .05       0    4226      .1       0  4372.9     .05       0
    4772      .1       0  5005.2     .07       0  5011.2      .1       0
    5077     .16       0  5184.3     .05       0
Bank Sta=4975.6,5059.2
XS Rating Curve= 0 ,0
Exp/Cntr=0.3,0.1

Type RM Length L Ch R = 1 ,14456   ,1104,1104,1104
BEGIN DESCRIPTION:
SALT CREEK 1 25.0
END DESCRIPTION:
XS GIS Cut Line= 2
      3499674.61     10611448.66      3499716.27     10609920.83
#Sta/Elev= 30
    3937  453.79  4185.6  451.14  4240.5  444.42  4295.6  442.93  4307.3  447.59
  4355.6  440.53  4375.6  445.46  4385.6  441.31  4395.6  445.86  4445.7  438.84
  4455.7  446.89  4465.7  447.96  4515.7  442.29  4555.7  448.85  4632.5  448.91
  4730.5  448.27  4965.9  449.49  4975.9  441.55  5002.9  435.52  5005.6  435.02
  5008.9  435.52  5024.5  441.19  5045.9  446.89  5122.5  449.12  5155.9  448.31
  5220.6  456.27    5296  462.96    5316  458.82  5416.6  469.11  5465.4  475.38
#Mann= 10 ,-1 , 0
    3937     .05       0  4240.5     .16       0  4632.5      .1       0
  4730.5     .16       0  5002.9     .07       0  5008.9     .16       0
  5024.5      .1       0  5122.5     .05       0  5220.6     .16       0
  5416.6     .05       0
Bank Sta=4965.9,5045.9
XS Rating Curve= 0 ,0
Exp/Cntr=0.3,0.1

Type RM Length L Ch R = 1 ,13352   ,299,299,299
BEGIN DESCRIPTION:
SALT CREEK 1 23.0
END DESCRIPTION:
XS GIS Cut Line= 2
      3500306.55     10611490.31      3500216.28     10610150.05
#Sta/Elev= 30
  4354.9  452.28  4445.2  451.45  4475.3  449.23  4505.4  450.13  4531.5  448.26
  4555.5  449.15  4686.1  446.58  4736.4  447.38  4936.3  445.69  4975.2  441.24
  4980.2  443.54  4993.5  433.38  4996.2  432.88  4999.5  433.38  5006.5  435.93
  5026.5  436.97  5036.6  442.86  5046.6  445.57  5066.6  440.54    5071  440.78
  5116.7  441.82  5136.8  444.27  5146.8  446.85    5217  449.56  5366.7  450.86
  5447.5  453.03  5477.6   456.1  5564.2   460.3  5644.4  463.57  5698.2  467.77
#Mann= 8 ,-1 , 0
  4354.9     .16       0  4736.4     .05       0  4993.5    .035       0
  4999.5     .05       0    5071     .16       0  5366.7     .05       0
  5564.2      .1       0  5644.4     .05       0
Bank Sta=4993.5,4999.5
XS Rating Curve= 0 ,0
Exp/Cntr=0.3,0.1

Type RM Length L Ch R = 1 ,13053   ,484,484,484
BEGIN DESCRIPTION:
SALT CREEK 1 22.0
END DESCRIPTION:
XS GIS Cut Line= 3
      3500699.61     10611960.22      3500499.61     10610760.19
      3500299.61     10609960.19
#Sta/Elev= 30
  3743.2  459.61    4183  452.13  4333.6  448.23  4413.9  447.73  4483.3  447.06
  4523.9  445.02  4554.3  446.33  4652.3  445.24  4764.8  446.15  4909.1  447.14
  4949.6  444.05  4957.2  440.22  4977.8  438.13  4990.7  433.19    4998  432.81
  5000.8  432.31    5004  432.81  5019.1  435.15  5024.2   439.5  5065.4  447.11
  5101.5  446.18  5239.9   449.7  5348.9  451.08  5444.2  454.91  5503.9  460.64
  5512.6  460.96    5519  462.47  5547.3  462.58  5567.9  465.45  5784.4  480.85
#Mann= 11 ,-1 , 0
  3743.2     .05       0    4183     .16       0  4333.6     .05       0
  4413.9     .16       0  4652.3     .05       0  4764.8     .16       0
    4998     .07       0    5004     .16       0  5239.9     .05       0
  5503.9      .1       0  5512.6     .05       0
Bank Sta=4998,5004
XS Rating Curve= 0 ,0
Exp/Cntr=0.3,0.1

Type RM Length L Ch R = 1 ,12569   ,985,985,985
BEGIN DESCRIPTION:
SALT CREEK 1 21.0
END DESCRIPTION:
XS GIS Cut Line= 3
      3501445.43     10611372.22      3500945.44     10611080.55
      3500778.77     10610038.85
#Sta/Elev= 30
  3863.6  455.57  3886.6  455.23  4078.4  449.73  4197.7  445.55  4219.2  442.05
  4229.1  445.35  4240.8   445.5  4293.6  442.49  4309.3  445.16  4402.9  444.81
    4426  441.56  4452.9  445.55  4908.7  445.94    4939  442.68  4954.1  444.63
  4969.4   442.5  4979.6  438.26  4989.7  436.82  4996.8  432.08  4999.6  431.58
  5002.8  432.08  5025.2   433.4  5030.2  434.77  5040.3  446.65  5111.2  445.84
  5303.6  455.79  5331.4  458.64  5364.4  459.03  5393.4  463.72  5497.4  473.76
#Mann= 6 ,-1 , 0
  3863.6      .1       0  3886.6     .05       0  4078.4     .16       0
  4996.8     .07       0  5002.8     .16       0  5025.2     .05       0
Bank Sta=4996.8,5002.8
XS Rating Curve= 0 ,0
Exp/Cntr=0.3,0.1

Type RM Length L Ch R = 1 ,11584   ,376,376,376
BEGIN DESCRIPTION:
SALT CREEK 1 20.0
END DESCRIPTION:
XS GIS Cut Line= 3
      3501647.05     10611233.78      3501532.46     10610785.85
      3501053.98     10610198.15
#Sta/Elev= 30
  4676.2  454.31  4690.7  452.88  4726.4  453.16  4789.6  451.15  4848.8  447.35
  4884.5  446.96  4889.6  445.78  4925.3  444.86  4930.5  443.24  4948.3  440.81
  4979.2  437.93  4989.6  429.99  4994.1  429.92  4996.9  429.88  4999.6  429.38
  5002.9  429.88  5012.1  432.44  5020.5  436.16  5030.9  438.08  5041.2  441.29
  5072.1  441.54  5096.4   443.5  5129.4  442.59  5151.6   444.4  5314.7  442.91
  5372.1  444.05  5429.5  443.14  5528.7   444.1  5713.2  447.12  5896.4   452.3
#Mann= 6 ,-1 , 0
  4676.2     .16       0  4789.6     .05       0  4994.1     .16       0
  4996.9     .07       0  5002.9     .16       0  5096.4     .05       0
Bank Sta=4996.9,5002.9
XS Rating Curve= 0 ,0
Exp/Cntr=0.3,0.1

Type RM Length L Ch R = 1 ,11208   ,685,685,685
BEGIN DESCRIPTION:
SALT CREEK 1 19.0
END DESCRIPTION:
XS GIS Cut Line= 3
      3501849.61     10611110.24      3501799.61     10610660.19
       3500999.6     10609860.18
#Sta/Elev= 30
  4528.2  455.15  4604.2  453.21    4659     452  4709.4  449.34  4779.8  449.11
  4802.5  447.35    4820  446.11  4830.1  443.76  4850.2  441.66  4870.3  441.21
  4890.5  443.52  4940.8  443.66  4960.9   439.9    4971   435.3  4984.6  435.18
  4995.2  430.94  5006.3  430.05  5009.1  429.55  5012.3  430.05  5023.4  438.63
  5037.6  442.87  5048.3  442.83  5306.3  442.72  5631.6  447.89  5744.7  450.92
  5787.1  453.38  5801.3  455.61    5872  459.21  6013.4  471.26  6112.4  481.16
#Mann= 6 ,-1 , 0
  4528.2      .1       0  4604.2     .05       0  4802.5     .16       0
  5006.3     .07       0  5012.3     .16       0  5048.3     .05       0
Bank Sta=5006.3,5012.3
XS Rating Curve= 0 ,0
Exp/Cntr=0.3,0.1

Type RM Length L Ch R = 1 ,10523   ,894,894,894
BEGIN DESCRIPTION:
SALT CREEK 1 18.0
END DESCRIPTION:
XS GIS Cut Line= 2
      3502376.24      10610676.5      3501589.76     10609796.28
#Sta/Elev= 30
    4700  448.59    4723  449.25  4737.2  445.42  4808.3  439.71  4822.5   441.6
  4836.7  438.95  4843.4  435.59  4850.9  436.82  4865.1  434.44  4871.8  440.69
  4942.9  442.32  4949.9  441.72  4957.1  437.09  4963.8  435.26    4978  434.59
  4985.5  430.45  4996.7  430.05  4999.5  429.55  5002.7  430.05  5006.4  431.32
  5013.9  439.42  5028.1  442.81  5234.1  442.35  5254.7  444.15  5289.8  442.19
  5473.7  442.03    5630  443.96  5714.5  446.75  5757.1  451.85  5880.4  459.98
#Mann= 4 ,-1 , 0
    4700     .16       0  4996.7     .07       0  5002.7     .16       0
  5234.1     .05       0
Bank Sta=4996.7,5002.7
XS Rating Curve= 0 ,0
Exp/Cntr=0.3,0.1

Type RM Length L Ch R = 1 ,9629    ,425,425,425
BEGIN DESCRIPTION:
SALT CREEK 1 16.0
END DESCRIPTION:
XS GIS Cut Line= 3
      3503099.61     10611060.18      3502399.61     10609860.19
      3501799.59     10609260.17
#Sta/Elev= 30
  3604.3  455.61  3655.2  456.14  3831.3  451.59  4102.1  450.48  4136.8  448.57
    4160  449.55  4424.2  445.16    4430  443.93    4473  445.45  4621.5  441.78
  4750.3  440.68  4765.6  440.74  4782.3  440.59  4809.5  437.29    4841  439.99
  4846.8  441.83  4921.2  441.12  4948.5  437.88  4970.4  437.38  4990.6  430.25
  5004.7  428.39  5007.4  427.89  5010.7  428.39  5026.4  434.72    5036  438.32
  5050.1  440.26  5318.8  442.74  5559.2  450.04  5785.5  467.34  5842.1  468.78
#Mann= 7 ,-1 , 0
  3604.3     .05       0  4621.5     .16       0  4750.3     .05       0
  4765.6     .16       0  5004.7     .07       0  5010.7     .16       0
  5026.4     .05       0
Bank Sta=5004.7,5010.7
XS Rating Curve= 0 ,0
Exp/Cntr=0.3,0.1

Type RM Length L Ch R = 1 ,9204    ,486,486,486
BEGIN DESCRIPTION:
SALT CREEK 1 15.0
END DESCRIPTION:
XS GIS Cut Line= 3
       3503362.1      10610750.7      3502761.43     10609629.21
      3502043.68     10609199.25
#Sta/Elev= 30
  3673.2  453.34  3843.9   451.8  3985.7  448.26  4171.7  446.25  4193.7  444.47
  4243.2  444.39  4310.6  441.45  4410.9   439.2    4518  438.86  4638.2   439.2
  4850.9  439.17  4872.9  437.61  4894.8  438.26  4900.5   436.8  4908.1  437.87
  4916.7  439.49  4949.3   438.1  4990.3  428.64  4993.1  426.01  4995.8  425.51
  4999.1  426.01  5017.5  426.91    5033  438.53  5122.4  437.69  5149.2  439.85
  5303.3  440.45  5515.2  444.29  5674.7  450.32  5690.2  452.31  5782.1  456.88
#Mann= 9 ,-1 , 0
  3673.2     .05       0  4310.6     .16       0  4410.9     .05       0
    4518     .16       0  4638.2     .05       0  4908.1     .16       0
  4993.1     .07       0  4999.1     .16       0  5149.2     .05       0
Bank Sta=4949.3,5033
XS Rating Curve= 0 ,0
Exp/Cntr=0.3,0.1

Type RM Length L Ch R = 1 ,8718    ,499,499,499
BEGIN DESCRIPTION:
SALT CREEK 1 14.0
END DESCRIPTION:
XS GIS Cut Line= 3
      3503511.56     10610627.99      3503045.05     10609311.46
      3502303.25     10609149.14
#Sta/Elev= 30
  3654.8  452.57  3826.4  451.74    3950  448.97  4023.8   450.5  4342.1  438.85
  4522.4  437.08  4623.4  438.27  4633.8  439.88  4639.1  438.49  4681.6   436.3
  4690.2  437.95  4721.1  438.72  4819.5  437.47  4906.4  438.26  4931.2   436.5
    4940  436.11  4946.8  436.05  4957.4  429.09  4959.9  424.23  4962.6  423.73
  4965.9  424.23  4978.6  426.93  4993.8  427.32  4999.8  424.98  5010.5  426.86
  5019.3  438.31  5218.5  438.46  5407.8  441.44  5630.4  443.15  5810.9  448.47
#Mann= 7 ,-1 , 0
  3654.8     .05       0  4623.4     .16       0  4931.2     .05       0
    4940     .16       0  4959.9     .07       0  4965.9     .16       0
  5407.8     .05       0
Bank Sta=4946.8,5019.3
XS Rating Curve= 0 ,0
Exp/Cntr=0.3,0.1

Type RM Length L Ch R = 1 ,8219    ,310,310,310
BEGIN DESCRIPTION:
Mapping XS a4e463ed
END DESCRIPTION:
XS GIS Cut Line= 3
      3504264.87      10610226.4      3503494.06     10609358.38
      3502219.72     10608709.05
#Sta/Elev= 30
  3901.2  450.51  4031.6  450.06  4220.8  447.86  4263.5   450.3  4320.3  442.97
  4369.7  445.26  4439.9  443.79  4539.4  441.16  4567.9  442.73  4686.8  441.39
    4792  439.71  4822.8  438.71  4957.6  436.39  4965.1  436.04  4979.3  426.19
  5003.9   424.6  5006.7   424.1  5009.9   424.6  5014.4   427.9  5021.1  426.66
  5028.7  434.65  5057.1  437.23  5352.5  438.36  5532.2  440.89  5576.7  438.86
  5740.5  438.96  5821.3  440.35  5843.5  442.65  6193.7  445.19  6492.3  458.57
#Mann= 9 ,-1 , 0
  3901.2     .05       0  4031.6     .16       0  4439.9     .05       0
  4686.8     .16       0    4792      .1       0  4822.8     .16       0
  5003.9     .07       0  5009.9     .16       0  5352.5     .05       0
Bank Sta=4957.6,5057.1
XS Rating Curve= 0 ,0
Exp/Cntr=0.3,0.1

Type RM Length L Ch R = 1 ,7909    ,107,107,107
BEGIN DESCRIPTION:
SALT CREEK 1 13.0
END DESCRIPTION:
XS GIS Cut Line= 3
      3504403.56     10609307.12      3503629.48     10609254.21
        3502567.     10608427.84
#Sta/Elev= 30
  4394.7  445.78  4498.9  446.02  4739.5  441.91  4749.5  440.57  4849.7  440.02
  4879.8  437.37  4949.9  435.57    4960  433.93    4987  423.17  4989.8  422.67
    4993  423.17  5012.3  424.79  5020.1  427.19  5040.2  426.05  5060.2  429.47
  5070.2   436.1  5114.5  436.56  5150.4  434.36  5160.8  437.01  5191.3  436.87
  5558.4   436.5  5579.2  434.77  5622.6  436.82  5715.2  436.46  5728.5  438.53
  5979.1  438.28  6242.5  444.85  6327.5  448.46  6362.8  451.88  6516.6  456.96
#Mann= 5 ,-1 , 0
  4394.7     .16       0    4987     .07       0    4993     .16       0
  5114.5      .1       0  5191.3     .05       0
Bank Sta=4949.9,5070.2
XS Rating Curve= 0 ,0
Exp/Cntr=0.3,0.1

Type RM Length L Ch R = 1 ,7802    ,508,508,508
BEGIN DESCRIPTION:
SALT CREEK 1 12.0
END DESCRIPTION:
XS GIS Cut Line= 3
       3504629.5     10609209.07      3503621.09     10609161.98
       3502639.9     10608365.32
#Sta/Elev= 30
  4218.5  445.33  4270.3  445.33  4708.9  440.24    4819  440.31  4839.1  439.12
  4849.1   434.6  4869.1  431.55  4899.1  431.33  4939.2  434.23  4969.2  430.34
  4979.2  423.24  4996.2  421.84    4999  421.34  5002.2  421.84  5039.3  433.47
  5059.3  436.34  5307.9   435.2  5443.7  436.35  5486.9  434.08  5528.5  436.25
  5763.4  436.76  5777.8  438.57  5792.2  437.41  5905.6  437.64  6225.3  444.21
  6268.4  446.38  6289.2  449.61  6396.3  453.14  6431.5   455.7  6491.9  455.79
#Mann= 4 ,-1 , 0
  4218.5     .08       0  4270.3     .05       0  4996.2     .04       0
  5002.2     .05       0
Bank Sta=4939.2,5059.3
XS Rating Curve= 0 ,0
Exp/Cntr=0.3,0.1
