--- TEHUACANA CREEK.prj (project) ---

Proj Title=TEHUACANA CREEK Base Level Engineering
Current Plan=p01
Default Exp/Contr=0.3,0.1
English Units
Geom File=g01
Flow File=f01
Plan File=p01
Y Axis Title=Elevation
X Axis Title(PF)=Main Channel Distance
X Axis Title(XS)=Station
BEGIN DESCRIPTION:
TEHUACANA CREEK
END DESCRIPTION:
DSS Export Rating Curves= 0
DSS Export Rating Curve Sorted= 0
DSS Export Volume Flow Curves= 0
DXF OffsetX= 0
DXF OffsetY= 0
DXF ScaleX= 1
DXF ScaleY= 10

--- TEHUACANA CREEK.p01 (plan) ---

Plan Title=Multiple Run
Short Identifier=Multiple
Geom File=g01
Flow File=f01
Subcritical Flow
K Sum by GR= 0
Std Step Tol= 0.01
Critical Tol= 0.01
Num of Std Step Trials= 20
Max Error Tol= 0.3
Flow Tol Ratio= 0.001
Split Flow NTrial= 30
Split Flow Tol= 0.02
Split Flow Ratio= 0.02
Log Output Level= 0
Friction Slope Method= 1
Unsteady Friction Slope Method= 2
Unsteady Bridges Friction Slope Method= 1
Parabolic Critical Depth
Global Vel Dist=  1 , 1 , 1
Global Log Level= 0
CheckData=True
Encroach Param= -1, 0, 0, 0
BEGIN DESCRIPTION:
Multiple Run
END DESCRIPTION:

--- TEHUACANA CREEK.f01 (steady flow) ---

Flow Title=Multiple
Program Version=4.10
Number of Profiles= 7
Profile Names=10-year,25-year,50-year,1pct_min,100-year,1pct_plu,500-year
River Rch & RM=TEHUACANA CREEK,Reach-1         ,312836
    2636    3812    4831    4460    6032    8158    9389
River Rch & RM=TEHUACANA CREEK,Reach-1         ,309219
    3101    4500    5714    5282    7143    9660   11145
River Rch & RM=TEHUACANA CREEK,Reach-1         ,302450
    3511    5109    6498    6012    8130   10995   12712
River Rch & RM=TEHUACANA CREEK,Reach-1         ,297733
    3785    5527    7046    6533    8836   11949   13874
River Rch & RM=TEHUACANA CREEK,Reach-1         ,294459
    5284    7785    9986    9302   12580   17013   19941
River Rch & RM=TEHUACANA CREEK,Reach-1         ,285270
    5527    8161   10482    9778   13223   17883   21016
River Rch & RM=TEHUACANA CREEK,Reach-1         ,284581
    5527    8161   10482    9778   13223   17883   21016
River Rch & RM=TEHUACANA CREEK,Reach-1         ,283044
    7126   10585   13652   12777   17279   23368   27639
River Rch & RM=TEHUACANA CREEK,Reach-1         ,282697
    7126   10585   13652   12777   17279   23368   27639
River Rch & RM=TEHUACANA CREEK,Reach-1         ,279197
    7359   10948   14135   13242   17909   24220   28706
River Rch & RM=TEHUACANA CREEK,Reach-1         ,276167
    7760   11561   14941   14009   18945   25621   30416
River Rch & RM=TEHUACANA CREEK,Reach-1         ,275482
    7760   11561   14941   14009   18945   25621   30416
River Rch & RM=TEHUACANA CREEK,Reach-1         ,273421
    7841   11657   15043   14081   19043   25753   30469
River Rch & RM=TEHUACANA CREEK,Reach-1         ,269456
    8137   12104   15625   14630   19785   26757   31670
River Rch & RM=TEHUACANA CREEK,Reach-1         ,264881
    8287   12301   15856   14820   20043   27105   31973
River Rch & RM=TEHUACANA CREEK,Reach-1         ,262772
    8287   12301   15856   14820   20043   27105   31973
River Rch & RM=TEHUACANA CREEK,Reach-1         ,257892
   18496   28058   36725   34804   47069   63655   77127
River Rch & RM=TEHUACANA CREEK,Reach-1         ,253464
   18496   28058   36725   34804   47069   63655   77127
River Rch & RM=TEHUACANA CREEK,Reach-1         ,250752
   18496   28058   36725   34804   47069   63655   77127
River Rch & RM=TEHUACANA CREEK,Reach-1         ,246037
   18736   28405   37164   35204   47610   64386   77937
River Rch & RM=TEHUACANA CREEK,Reach-1         ,243927
   18736   28405   37164   35204   47610   64386   77937
River Rch & RM=TEHUACANA CREEK,Reach-1         ,240569
   19614   29741   38920   36870   49862   67433   81629
River Rch & RM=TEHUACANA CREEK,Reach-1         ,237539
   19815   30046   39319   37248   50374   68125   82466
River Rch & RM=TEHUACANA CREEK,Reach-1         ,236850
   19815   30046   39319   37248   50374   68125   82466
River Rch & RM=TEHUACANA CREEK,Reach-1         ,228645
   19815   30046   39319   37248   50374   68125   82466
River Rch & RM=TEHUACANA CREEK,Reach-1         ,224068
   20634   31121   40577   38287   51779   70026   84078
River Rch & RM=TEHUACANA CREEK,Reach-1         ,215676
   20634   31121   40577   38287   51779   70026   84078
River Rch & RM=TEHUACANA CREEK,Reach-1         ,214529
   24482   37004   48329   45665   61757   83519  100534
River Rch & RM=TEHUACANA CREEK,Reach-1         ,206546
   29170   44073   57559   54371   73530   99441  119578
River Rch & RM=TEHUACANA CREEK,Reach-1         ,204446
   29170   44073   57559   54371   73530   99441  119578
River Rch & RM=TEHUACANA CREEK,Reach-1         ,196031
   29170   44073   57559   54371   73530   99441  119578
River Rch & RM=TEHUACANA CREEK,Reach-1         ,189255
   29170   44073   57559   54371   73530   99441  119578
River Rch & RM=TEHUACANA CREEK,Reach-1         ,187775
   29170   44073   57559   54371   73530   99441  119578
River Rch & RM=TEHUACANA CREEK,Reach-1         ,181711
   29170   44073   57559   54371   73530   99441  119578
River Rch & RM=TEHUACANA CREEK,Reach-1         ,179885
   29170   44073   57559   54371   73530   99441  119578
River Rch & RM=TEHUACANA CREEK,Reach-1         ,174696
   29170   44073   57559   54371   73530   99441  119578
River Rch & RM=TEHUACANA CREEK,Reach-1         ,173560
   29170   44073   57559   54371   73530   99441  119578
River Rch & RM=TEHUACANA CREEK,Reach-1         ,167385
   29170   44073   57559   54371   73530   99441  119578
River Rch & RM=TEHUACANA CREEK,Reach-1         ,162940
   30180   45352   59013   55528   75095  101557  121150
River Rch & RM=TEHUACANA CREEK,Reach-1         ,158624
   40101   60287   78515   73923   99973  135201  161362
River Rch & RM=TEHUACANA CREEK,Reach-1         ,157152
   40101   60287   78515   73923   99973  135201  161362
River Rch & RM=TEHUACANA CREEK,Reach-1         ,150374
   40101   60287   78515   73923   99973  135201  161362
River Rch & RM=TEHUACANA CREEK,Reach-1         ,148895
   41334   61942   80500   75623  102272  138311  164313
River Rch & RM=TEHUACANA CREEK,Reach-1         ,142109
   41334   61942   80500   75623  102272  138311  164313
River Rch & RM=TEHUACANA CREEK,Reach-1         ,128694
   41334   61942   80500   75623  102272  138311  164313
River Rch & RM=TEHUACANA CREEK,Reach-1         ,127287
   41334   61942   80500   75623  102272  138311  164313
River Rch & RM=TEHUACANA CREEK,Reach-1         ,121800
   41334   61942   80500   75623  102272  138311  164313
River Rch & RM=TEHUACANA CREEK,Reach-1         ,116306
   41529   62155   80709   75752  102446  138546  164313
River Rch & RM=TEHUACANA CREEK,Reach-1         ,109998
   41574   62166   80709   75752  102446  138546  164313
River Rch & RM=TEHUACANA CREEK,Reach-1         ,108339
   41746   62405   80967   75929  102686  138870  164391
River Rch & RM=TEHUACANA CREEK,Reach-1         ,106890
   41746   62405   80967   75929  102686  138870  164391
River Rch & RM=TEHUACANA CREEK,Reach-1         ,98904
   41746   62405   80967   75929  102686  138870  164391
River Rch & RM=TEHUACANA CREEK,Reach-1         ,97429
   41746   62405   80967   75929  102686  138870  164391
River Rch & RM=TEHUACANA CREEK,Reach-1         ,91239
   41746   62405   80967   75929  102686  138870  164391
River Rch & RM=TEHUACANA CREEK,Reach-1         ,88818
   45771   68128   88154   82432  111480  150764  177385
River Rch & RM=TEHUACANA CREEK,Reach-1         ,85492
   45771   68128   88154   82432  111480  150764  177385
River Rch & RM=TEHUACANA CREEK,Reach-1         ,81722
   45771   68128   88154   82432  111480  150764  177385
River Rch & RM=TEHUACANA CREEK,Reach-1         ,73065
   45771   68128   88154   82432  111480  150764  177385
River Rch & RM=TEHUACANA CREEK,Reach-1         ,68139
   47738   71102   92052   86123  116472  157515  185512
River Rch & RM=TEHUACANA CREEK,Reach-1         ,63596
   47738   71102   92052   86123  116472  157515  185512
River Rch & RM=TEHUACANA CREEK,Reach-1         ,57358
   47746   71102   92052   86123  116472  157515  185512
River Rch & RM=TEHUACANA CREEK,Reach-1         ,40819
   47996   71321   92193   86123  116472  157515  185512
River Rch & RM=TEHUACANA CREEK,Reach-1         ,36188
   48399   71896   92916   86772  117350  158702  186205
River Rch & RM=TEHUACANA CREEK,Reach-1         ,35229
   48399   71896   92916   86772  117350  158702  186205
River Rch & RM=TEHUACANA CREEK,Reach-1         ,25674
   48399   71896   92916   86772  117350  158702  186205
River Rch & RM=TEHUACANA CREEK,Reach-1         ,9995
   51193   75832   97833   91201  123338  166801  194973
Boundary for River Rch & Prof#=TEHUACANA CREEK,Reach-1         , 1
Up Type= 0
Dn Type= 3
Dn Slope=0.00059
Boundary for River Rch & Prof#=TEHUACANA CREEK,Reach-1         , 2
Up Type= 0
Dn Type= 3
Dn Slope=0.00059
Boundary for River Rch & Prof#=TEHUACANA CREEK,Reach-1         , 3
Up Type= 0
Dn Type= 3
Dn Slope=0.00059
Boundary for River Rch & Prof#=TEHUACANA CREEK,Reach-1         , 4
Up Type= 0
Dn Type= 3
Dn Slope=0.00059
Boundary for River Rch & Prof#=TEHUACANA CREEK,Reach-1         , 5
Up Type= 0
Dn Type= 3
Dn Slope=0.00059
Boundary for River Rch & Prof#=TEHUACANA CREEK,Reach-1         , 6
Up Type= 0
Dn Type= 3
Dn Slope=0.00059
Boundary for River Rch & Prof#=TEHUACANA CREEK,Reach-1         , 7
Up Type= 0
Dn Type= 3
Dn Slope=0.00059
DSS Import GetInterval= 0
DSS Import GetPeak= 0
DSS Import FillOption= 0

--- TEHUACANA CREEK.g01 (geometry) ---

Geom Title=Existing Conditions
Program Version=4.10

River Reach=TEHUACANA CREEK ,Reach-1
Reach XY= 30
       3478846.5       10614909.      3488942.75       10622325.
      3492855.25       10619202.      3508868.25       10620254.
        3518939.       10627690.        3526963.       10643819.
      3536573.25       10654433.       3545889.5       10657621.
        3548434.       10656342.        3555269.       10659937.
      3563218.25       10659653.        3568152.       10663873.
      3569866.75       10669195.        3574752.       10669155.
       3577879.5       10672910.      3582986.25       10674013.
       3583406.5       10676005.      3589971.25       10679067.
      3594967.25       10678650.       3596493.5       10683182.
      3604805.25       10686139.       3605966.5       10683044.
       3619967.5       10679423.        3627257.       10666295.
        3630252.       10664624.       3635191.5       10666806.
      3636553.75       10663618.      3641284.75       10662209.
        3641602.       10656813.       3648965.3     10655226.66

Type RM Length L Ch R = 1 ,312836  ,442,442,442
BEGIN DESCRIPTION:
TEHUACANA CREEK 259.0
END DESCRIPTION:
XS GIS Cut Line= 3
      3477799.59     10615110.19      3478999.61     10615310.19
       3479299.6     10615260.19
#Sta/Elev= 30
  3805.6  529.33  3866.4  526.97  4251.7  521.86  4325.2  520.02  4434.2  519.22
  4563.4  516.26    4634  516.05  4690.2  515.83  4707.9  514.33  4738.3  516.54
  4778.9  515.63    4789  517.18  4799.1   517.2  4806.7  516.22  4811.8  516.62
  4872.6  515.26  4900.5  516.18  4971.5  516.02  4989.2  515.62  5001.9  514.51
    5009  512.31  5011.8  511.81    5015  512.31  5019.6  515.69  5032.3  516.03
  5072.9  515.52  5133.6  517.32  5245.2  521.34  5255.3  522.38  5326.3  525.74
#Mann= 5 ,-1 , 0
  3805.6     .05       0    4634     .16       0    5009     .07       0
    5015     .16       0  5133.6     .05       0
Bank Sta=4971.5,5032.3
XS Rating Curve= 0 ,0
Exp/Cntr=0.3,0.1

Type RM Length L Ch R = 1 ,312394  ,471,471,471
BEGIN DESCRIPTION:
TEHUACANA CREEK 258.0
END DESCRIPTION:
XS GIS Cut Line= 2
      3478060.49      10615421.4      3479741.02     10615876.26
#Sta/Elev= 30
  3945.4  522.57  4377.7   515.5  4622.5  513.58    4680  513.63  4686.2  511.77
  4691.4  512.55  4700.8   509.2  4711.1  513.35  4752.6  512.36  4875.1  513.59
  4897.6  512.33  4980.5  513.35  4989.5  511.35  4994.7  511.41  4998.2  509.02
  5000.9  508.52  5004.2  509.02  5011.5  512.36  5021.9  513.37  5042.6  512.88
    5063   514.2  5069.2  514.42  5074.4  512.56  5094.4  514.02  5166.9  515.64
    5198  517.63    5298  520.11  5519.2  524.98  5581.3  524.65  5686.4     530
#Mann= 5 ,-1 , 0
  3945.4     .05       0  4622.5     .16       0  4998.2     .07       0
  5004.2     .16       0    5063     .05       0
Bank Sta=4980.5,5069.2
XS Rating Curve= 0 ,0
Exp/Cntr=0.3,0.1

Type RM Length L Ch R = 1 ,311923  ,99,99,99
BEGIN DESCRIPTION:
TEHUACANA CREEK 257.0
END DESCRIPTION:
XS GIS Cut Line= 2
      3478011.88     10616042.93      3479782.72     10616056.81
#Sta/Elev= 30
  3768.8  520.38  3916.5  517.68  4016.5  517.79  4406.6  513.53  4676.6  512.15
  4696.6  513.31  4796.6   511.3  4836.6  511.26  4936.6  509.02  4966.6  507.47
  5003.6  503.82  5006.3  503.32  5009.6  503.82  5016.6  506.68  5026.6  507.58
  5046.6  506.89  5056.6  510.69  5066.6  511.26  5076.6  512.72  5136.6  514.29
  5146.6  515.58  5166.6  515.08  5186.6  515.71  5216.6  515.46  5266.6  517.49
  5276.6  517.13  5296.6  518.35    5337  518.68  5406.6  520.65  5539.7  527.32
#Mann= 3 ,-1 , 0
  3768.8     .05       0  5003.6     .03       0  5009.6     .05       0
Bank Sta=4796.6,5076.6
XS Rating Curve= 0 ,0
Exp/Cntr=0.3,0.1

Type RM Length L Ch R = 1 ,311824  ,426,426,426
BEGIN DESCRIPTION:
TEHUACANA CREEK 256.0
END DESCRIPTION:
XS GIS Cut Line= 2
      3478025.73     10616147.09      3479764.93     10616150.56
#Sta/Elev= 30
  3770.6   521.6  4074.5   518.9  4134.5  517.24  4324.5  515.19  4344.5   514.5
  4394.5  515.02  4524.5  513.14  4554.5  513.49  4644.5  512.38  4674.5  511.38
  4824.5  511.21  4854.5  510.49  4954.5  509.81  4974.5  509.25  4984.5  505.49
  4991.5  501.76  4994.2  501.26  4997.5  501.76  5014.5  509.01  5044.5     509
  5074.5  509.83  5124.5  510.94  5144.5  512.32  5154.5  511.68  5184.5   511.7
  5254.5  515.71  5274.5  515.58  5354.5  518.46  5404.5  520.98  5509.8  523.51
#Mann= 3 ,-1 , 0
  3770.6     .05       0  4991.5     .04       0  4997.5     .05       0
Bank Sta=4954.5,5074.5
XS Rating Curve= 0 ,0
Exp/Cntr=0.3,0.1

Type RM Length L Ch R = 1 ,311398  ,626,626,626
BEGIN DESCRIPTION:
TEHUACANA CREEK 255.0
END DESCRIPTION:
XS GIS Cut Line= 2
      3478452.81     10617101.97      3480018.84     10616157.49
#Sta/Elev= 30
  3793.8  521.19  3813.4  520.05  3895.2  519.07  4222.1  516.14  4251.8  514.88
  4463.4  510.53    4543  510.25  4680.8  508.18    4776  508.54  4871.1  506.79
  4886.6  506.84    4908  508.33  4966.2  507.88    4972  504.52  5000.1  501.92
  5002.8  501.42  5006.1  501.92  5024.4  506.39  5045.8   507.8  5109.9  507.64
  5177.8  509.48  5220.5  511.55  5352.5  515.16  5410.8  518.06  5432.1  517.54
    5469  518.76  5474.8  519.96  5548.6  522.47    5570   524.2  5622.6  526.48
#Mann= 3 ,-1 , 0
  3793.8     .05       0  5000.1    .035       0  5006.1     .05       0
Bank Sta=4908,5177.8
XS Rating Curve= 0 ,0
Exp/Cntr=0.3,0.1

Type RM Length L Ch R = 1 ,310772  ,429,429,429
BEGIN DESCRIPTION:
TEHUACANA CREEK 254.0
END DESCRIPTION:
XS GIS Cut Line= 3
      3478937.78     10617386.68      3479937.79     10616865.84
       3480284.8     10616157.94
#Sta/Elev= 30
  3679.8  515.09  3862.3  514.15  3929.9  512.92  3944.8  513.48  4198.7  510.84
  4211.8  510.14  4226.5  510.71  4436.2  507.28  4568.8  504.17  4730.4  506.24
  4805.5  505.27  4888.5  507.17    4939  503.76  4978.5  505.33    4984  505.21
  4988.8  497.42  4991.6  496.92  4994.8  497.42  5006.5  498.69  5014.1  503.09
    5029  502.15  5036.4  504.89    5119   506.5  5282.1  510.37  5381.6  513.54
    5389  514.74  5403.9  514.73    5434  516.61    5552  518.71  5595.7   520.7
#Mann= 3 ,-1 , 0
  3679.8     .05       0  4988.8    .035       0  4994.8     .05       0
Bank Sta=4978.5,5119
XS Rating Curve= 0 ,0
Exp/Cntr=0.3,0.1

Type RM Length L Ch R = 1 ,310343  ,521,521,521
BEGIN DESCRIPTION:
TEHUACANA CREEK 253.0
END DESCRIPTION:
XS GIS Cut Line= 3
      3479375.29     10617615.85       3480423.9      10616921.4
      3480500.29      10616108.9
#Sta/Elev= 30
  3859.8  511.99  4076.6     509  4127.8  508.96  4154.8  509.72  4401.5  507.15
  4428.7  508.21  4437.6  507.32  4560.6  503.72    4588  503.94  4618.1  502.91
  4747.5  504.28  4870.8  502.91  4897.9  504.12  4949.1  501.71  4979.2  503.02
  4985.2  501.46  4997.2  495.79    5000  495.29  5003.2  495.79  5006.2  500.09
  5015.3  503.25  5064.4  502.44  5219.2  503.81  5530.5  508.11  5560.7  509.76
  5610.9  510.68  5751.5  515.66  5766.3   515.5  5912.2  521.52  5933.6   521.6
#Mann= 3 ,-1 , 0
  3859.8     .05       0  4997.2    .035       0  5003.2     .05       0
Bank Sta=4897.9,5015.3
XS Rating Curve= 0 ,0
Exp/Cntr=0.3,0.1

Type RM Length L Ch R = 1 ,309822  ,603,603,603
BEGIN DESCRIPTION:
TEHUACANA CREEK 252.0
END DESCRIPTION:
XS GIS Cut Line= 3
      3479799.62     10618260.18      3480799.61     10617060.19
       3480649.6     10616260.16
#Sta/Elev= 30
  3407.6  516.03  3435.6  513.45  3443.4  511.47  3478.5  510.03  4383.6  504.83
  4442.7  502.62    4473  502.95  4565.5  500.22  4592.8  501.41  4664.4  501.51
  4707.3  499.41    4749  501.42  4785.4  500.34  4813.4  501.64  4921.4  501.06
    4956  500.11  4969.6  500.97  4979.8   500.1    4990  495.52  4992.9  492.46
  4995.7  491.96  4998.9  492.46  5010.3  495.41  5020.5  499.76  5030.7  500.97
  5040.9  499.92  5053.6  501.43  5065.5  501.03  5431.7  505.77  5783.6  516.13
#Mann= 7 ,-1 , 0
  3407.6     .05       0  4383.6     .16       0  4442.7     .05       0
  4921.4     .16       0  4992.9     .07       0  4998.9     .16       0
  5065.5     .05       0
Bank Sta=4969.6,5030.7
XS Rating Curve= 0 ,0
Exp/Cntr=0.3,0.1

Type RM Length L Ch R = 1 ,309219  ,733,733,733
BEGIN DESCRIPTION:
TEHUACANA CREEK 251.0
END DESCRIPTION:
XS GIS Cut Line= 4
      3480423.93     10618122.76      3480951.68      10617671.4
      3481062.79     10617060.29      3480896.12     10616157.51
#Sta/Elev= 30
    4030  509.42  4099.9  507.83  4284.4  507.56  4405.1  505.64    4426  506.78
  4446.8  505.67  4624.7  504.15  4645.5  504.93  4667.5  503.84  4786.6  504.48
  4827.3  500.86  4878.1  499.33    4906  496.28  4949.3  499.44  4964.5  499.52
  4979.8  499.14  4989.9  497.51  4997.1  490.58  4999.8  490.08  5003.1  490.58
  5010.3  495.83  5017.8  499.27  5022.9   498.6  5040.7  499.69    5125  499.94
  5234.8  500.25  5299.9  500.12    5905  506.75  6189.7  512.18  6263.6  512.68
#Mann= 5 ,-1 , 0
    4030     .05       0  4997.1    .035       0  5003.1     .05       0
    5125     .16       0  5234.8     .05       0
Bank Sta=4964.5,5040.7
XS Rating Curve= 0 ,0
Exp/Cntr=0.3,0.1

Type RM Length L Ch R = 1 ,308486  ,441,441,441
BEGIN DESCRIPTION:
TEHUACANA CREEK 250.0
END DESCRIPTION:
XS GIS Cut Line= 3
      3480659.99     10618317.25      3481347.51     10617699.18
      3481666.96     10616525.57
#Sta/Elev= 30
  3932.3  507.79  3986.3  507.17    4008  508.24  4036.4  506.97  4199.3  505.92
  4312.2  506.96  4383.2  505.23  4404.1   506.6  4588.7  503.81  4609.7  505.02
  4709.1  502.79    4730   503.6  4744.2   502.4  4858.9  500.96  4882.7   497.7
  4928.3  494.77  4980.1  499.19  4990.5  498.33  4993.9  487.24  4996.6  486.74
  4999.9  487.24  5011.2  488.54  5021.6  496.77  5031.4  497.44  5042.3  496.39
  5094.1  497.97  5339.2  499.29  5458.5  501.23  5881.8  512.39  6073.1   514.4
#Mann= 3 ,-1 , 0
  3932.3     .05       0  4993.9    .035       0  4999.9     .05       0
Bank Sta=4980.1,5339.2
XS Rating Curve= 0 ,0
Exp/Cntr=0.3,0.1

Type RM Length L Ch R = 1 ,308045  ,1018,1018,1018
BEGIN DESCRIPTION:
TEHUACANA CREEK 249.0
END DESCRIPTION:
XS GIS Cut Line= 3
      3481149.61     10618310.18      3481699.61     10617510.19
       3481899.6     10617010.22
#Sta/Elev= 30
    4055   505.9  4285.6  504.89    4322  503.63  4343.2  504.89  4673.9  499.63
  4722.7  500.22  4737.6  499.53  4746.4  497.25  4767.4  494.53  4788.4  493.91
    4875  497.11  4904.5  494.52  4916.9  494.67  4961.6   497.2  4976.5  496.66
  4982.5   494.9  4989.4  486.89  4994.4  486.02  4997.2  485.52  5000.4  486.02
  5003.5  489.99  5012.1  495.55  5040.6  494.72  5089.1  496.19  5148.2  496.45
  5202.2  497.87  5363.7  501.03  5402.8  503.43  5417.6  502.92  5564.3  506.39
#Mann= 5 ,-1 , 0
    4055     .05       0  4994.4    .035       0  5000.4     .05       0
  5012.1     .16       0  5148.2     .05       0
Bank Sta=4961.6,5202.2
XS Rating Curve= 0 ,0
Exp/Cntr=0.3,0.1

Type RM Length L Ch R = 1 ,307027  ,674,674,674
BEGIN DESCRIPTION:
TEHUACANA CREEK 248.0
END DESCRIPTION:
XS GIS Cut Line= 3
      3481763.32     10618586.75      3482249.42     10617927.04
      3482304.96     10616864.86
#Sta/Elev= 30
  3861.1  502.47  4092.8  501.27  4155.5  500.04  4170.2  500.58  4370.7   496.4
  4606.7  494.59  4680.6  494.95  4737.5  492.27  4767.5  489.58  4797.6   490.4
  4847.6  493.95  4867.7  494.01  4927.8  493.44  4977.8   491.7  4987.8  490.33
  4994.7   483.4  4994.8   483.3  4997.6   482.8  5000.8   483.3  5007.9  484.23
  5017.9   489.8  5027.9  488.42  5037.9  491.96  5092.7  495.03    5098  495.72
  5458.5  501.09  5578.6  501.12  5608.7  502.35  5688.8  502.93  5744.2  504.88
#Mann= 5 ,-1 , 0
  3861.1     .05       0  4994.7     .16       0  4994.8     .07       0
  5000.8     .16       0  5092.7     .05       0
Bank Sta=4867.7,5098
XS Rating Curve= 0 ,0
Exp/Cntr=0.3,0.1

Type RM Length L Ch R = 1 ,306353  ,72,72,72
BEGIN DESCRIPTION:
TEHUACANA CREEK 247.0
END DESCRIPTION:
XS GIS Cut Line= 6
      3482783.63     10618773.47      3482993.39     10618180.44
      3482923.66     10618013.09      3482861.16     10617799.55
      3482835.12     10617690.17      3482767.52     10617284.57
#Sta/Elev= 30
  3956.9  503.86  4199.4  498.47    4611  494.46  4629.4  493.08  4634.9  494.94
  4658.7  492.18  4664.1  494.47  4711.8  491.37  4717.2  492.42  4802.1  491.51
  4812.2  489.47  4834.5  492.34  4861.6  491.75  4866.8  493.36  4940.6   493.1
  4975.1  491.42  4980.3  489.74  4986.9  481.44  4996.4  481.33  4999.1  480.83
  5002.4  481.33  5009.7   481.8  5030.2  489.98  5050.8  493.79  5157.5  492.44
  5193.4   491.7  5257.6   493.3  5357.7  497.02  5405.6  498.85  5513.4  500.69
#Mann= 7 ,-1 , 0
  3956.9     .05       0  4996.4    .035       0  5002.4     .05       0
  5157.5     .08       0  5257.6     .05       0  5357.7     .08       0
  5405.6     .05       0
Bank Sta=4940.6,5050.8
XS Rating Curve= 0 ,0
Exp/Cntr=0.3,0.1

Type RM Length L Ch R = 1 ,306281  ,631,631,631
BEGIN DESCRIPTION:
TEHUACANA CREEK 246.0
END DESCRIPTION:
XS GIS Cut Line= 6
      3482842.24     10618792.97      3483054.75     10618178.92
      3483006.99     10618070.38      3482975.74     10617981.84
      3482944.49     10617872.47       3482829.9     10617210.99
#Sta/Elev= 30
  3919.4  503.64  4155.1  498.59  4508.6  494.39    4569  495.14    4725  491.35
    4756  492.36    4821  487.77  4887.4  489.45  4907.9  492.11  4938.4  491.79
  4946.3  490.19  4951.4  492.91  4979.1  490.89  5000.9  479.84  5003.7  479.34
  5006.9  479.84  5040.2  488.99  5056.5  488.96  5061.3   491.6    5065   491.6
  5118.7  488.42  5123.7  489.73  5171.9  489.75  5332.8  496.87  5370.2  499.61
  5375.3  498.28  5433.2  498.92  5536.1  501.24  5541.2  499.47  5566.8  501.75
#Mann= 5 ,-1 , 0
  3919.4     .05       0  5000.9     .04       0  5006.9     .05       0
  5332.8     .08       0  5433.2     .05       0
Bank Sta=4951.4,5065
XS Rating Curve= 0 ,0
Exp/Cntr=0.3,0.1

Type RM Length L Ch R = 1 ,305650  ,1005,1005,1005
BEGIN DESCRIPTION:
TEHUACANA CREEK 245.0
END DESCRIPTION:
XS GIS Cut Line= 3
       3482949.6     10618810.21      3483349.61     10617610.19
      3483249.62     10617260.23
#Sta/Elev= 30
  3725.5  503.64  4010.1  497.79  4199.9  495.33  4220.9  496.65  4389.6  495.03
  4463.4   493.1  4708.7  490.51  4738.3  490.39    4778  489.84  4874.5  487.54
  4895.6   490.3  4906.1  489.26  4916.6  480.29  4937.7  485.21  4948.3  479.83
  4958.8  480.75  4969.4  485.05  4979.9  482.99  4984.8  478.61  4987.5  478.11
  4990.8  478.61  5000.8  478.63  5007.3  482.24  5012.5  481.15    5032   488.8
  5052.8  491.14  5146.4  490.71  5208.8  494.19  5294.6  496.54  5354.4  499.25
#Mann= 7 ,-1 , 0
  3725.5     .05       0  4708.7     .08       0  4738.3     .05       0
    4778     .16       0  4984.8     .07       0  4990.8     .16       0
  5294.6     .05       0
Bank Sta=4895.6,5052.8
XS Rating Curve= 0 ,0
Exp/Cntr=0.3,0.1

Type RM Length L Ch R = 1 ,304645  ,506,506,506
BEGIN DESCRIPTION:
TEHUACANA CREEK 244.0
END DESCRIPTION:
XS GIS Cut Line= 3
       3483349.6      10618210.2      3483949.61     10617310.19
      3483949.61     10617160.17
#Sta/Elev= 30
  3908.3  494.61  4399.6     490  4543.8  488.81  4549.8  490.67  4564.8  486.29
  4629.4  486.21    4679  490.94  4724.1  489.43  4748.3  490.52  4760.1  491.46
  4766.1  489.12  4787.2  486.21  4809.7   485.7  4893.2  483.63  4910.4  483.21
  4917.9  481.01  4925.4  484.19  4940.4   483.9  4946.4  481.01  4961.4  481.14
    4997  473.59  4999.7  473.09    5003  473.59    5010  473.77    5030  485.95
    5060  491.01    5090  493.53    5110  501.25    5120  501.49    5140  496.55
#Mann= 6 ,-1 , 0
  3908.3     .05       0  4399.6     .08       0  4748.3     .05       0
  4893.2     .16       0    4997     .07       0    5003     .16       0
Bank Sta=4809.7,5060
XS Rating Curve= 0 ,0
Exp/Cntr=0.3,0.1

Type RM Length L Ch R = 1 ,304139  ,880,880,880
BEGIN DESCRIPTION:
TEHUACANA CREEK 243.0
END DESCRIPTION:
XS GIS Cut Line= 2
      3483596.64     10618829.83      3484630.77     10616824.02
#Sta/Elev= 30
  3688.1  502.04  3890.2     496  4059.6  493.02  4441.5  490.08  4469.4  491.17
  4530.3  488.84  4610.3  488.24  4707.6  490.03  4774.1   488.3  4936.5  488.29
  4973.5  486.63  4981.5  483.16  4990.1   471.6    5001  470.76  5003.8  470.26
    5007  470.76  5017.9  473.03  5026.5  480.12    5040  484.59  5106.5  485.11
  5195.3  488.19  5233.9  489.86  5285.3  494.33  5322.5  495.64  5449.9  506.39
  5582.8  509.82  5599.4   512.2  5665.9  513.28  5848.8  508.29  5944.8  507.57
#Mann= 3 ,-1 , 0
  3688.1     .05       0    5001    .035       0    5007     .05       0
Bank Sta=4936.5,5195.3
XS Rating Curve= 0 ,0
Exp/Cntr=0.3,0.1

Type RM Length L Ch R = 1 ,303259  ,809,809,809
BEGIN DESCRIPTION:
TEHUACANA CREEK 241.0
END DESCRIPTION:
XS GIS Cut Line= 3
       3483825.8     10618892.33      3484888.31     10617885.37
      3485298.01     10617309.01
#Sta/Elev= 30
  3467.6  497.88  3641.5  494.21  3959.8  490.14  4115.6  489.75  4419.8  484.62
  4547.2  484.67    4639  487.15  4716.7  486.65  4808.9  483.66    4851  485.25
    4892  484.28  4957.9  484.57  4972.7  483.25  4993.6  469.91  4996.7  468.89
  4999.5  468.39  5002.7  468.89  5008.3  473.38  5014.5  475.07  5023.1  483.64
  5050.1  480.86  5207.7  493.64  5273.9  496.82  5308.4  498.24  5323.2  499.97
  5355.4  500.55  5379.7  502.76  5464.3  505.26  5545.8  506.68  5638.6  505.26
#Mann= 7 ,-1 , 0
  3467.6     .05       0    4892     .16       0  4996.7     .07       0
  5002.7     .16       0  5273.9     .05       0  5355.4     .16       0
  5464.3     .05       0
Bank Sta=4957.9,5023.1
XS Rating Curve= 0 ,0
Exp/Cntr=0.3,0.1

Type RM Length L Ch R = 1 ,302450  ,535,535,535
BEGIN DESCRIPTION:
TEHUACANA CREEK 239.0
END DESCRIPTION:
XS GIS Cut Line= 2
      3484374.42      10618857.6      3486152.23     10617788.13
#Sta/Elev= 30
  3773.5     493  3929.4  489.66  4067.3  489.19  4162.5  487.05  4199.4  488.01
    4279  486.44  4321.8  484.12  4628.7  484.12  4655.9  487.13  4853.2   481.5
  4954.6  482.25  4962.8  482.82  4978.3  482.21  4984.2  475.21  4993.2   467.3
  4996.7  466.88  4999.5  466.38  5002.7  466.88  5015.2   471.2  5021.1  476.56
  5028.2     481    5058  481.49  5086.6  484.17  5185.8  491.55  5232.8  495.74
  5296.9  498.58  5349.3   497.8    5495   499.2  5693.2  502.91  5848.2  508.15
#Mann= 5 ,-1 , 0
  3773.5     .05       0  4954.6     .16       0  4996.7     .07       0
  5002.7     .16       0  5185.8     .05       0
Bank Sta=4962.8,5086.6
XS Rating Curve= 0 ,0
Exp/Cntr=0.3,0.1

Type RM Length L Ch R = 1 ,301915  ,458,458,458
BEGIN DESCRIPTION:
TEHUACANA CREEK 238.0
END DESCRIPTION:
XS GIS Cut Line= 2
      3484381.35     10618968.71      3486318.86     10618517.32
#Sta/Elev= 30
  3738.8  495.07  4116.9  487.49  4327.3  486.21    4579  482.28  4678.2  482.48
  4858.7  478.32  4876.7  473.11  4890.3  475.43  4896.2  477.16  4901.3  474.32
  4907.5  478.83  4979.4  480.24  4986.5  473.53  4991.6  473.02    5000  466.88
  5007.2  466.78    5010  466.28  5013.2  466.78  5020.5  475.86  5034.2  478.53
  5088.6  479.72  5161.9  481.41    5195  482.44  5236.1   487.8    5263  485.59
    5308  485.41  5337.3  490.44  5372.1  492.31  5595.5  506.64  5728.2  511.26
#Mann= 7 ,-1 , 0
  3738.8     .05       0  4890.3     .16       0  5007.2     .07       0
  5013.2     .16       0  5088.6     .05       0    5263     .16       0
  5372.1     .05       0
Bank Sta=4979.4,5161.9
XS Rating Curve= 0 ,0
Exp/Cntr=0.3,0.1

Type RM Length L Ch R = 1 ,301457  ,576,576,576
BEGIN DESCRIPTION:
TEHUACANA CREEK 237.0
END DESCRIPTION:
XS GIS Cut Line= 3
      3484492.45     10619135.37      3485728.59     10619086.76
      3486561.91     10618663.16
#Sta/Elev= 30
  3661.7  492.53  4039.1  486.39  4174.8   486.5  4199.3  484.79  4279.3  486.22
  4349.4  483.48  4449.5  482.46  4739.7  481.87  4869.8  475.26    4956  478.22
  4962.9  477.89  4978.5  476.79  4992.9  465.28  4997.9  465.06  5000.6  464.56
  5003.9  465.06  5009.6  467.92  5015.2  473.98  5023.3  472.64  5031.8  467.42
  5037.4  467.41  5045.8  468.78  5054.1  477.76  5090.6  479.27  5092.4  479.46
  5180.4  483.88  5321.1  494.86  5454.6  502.47  5699.4  507.62  5833.6  506.63
#Mann= 5 ,-1 , 0
  3661.7     .05       0  4962.9     .16       0  4997.9     .07       0
  5003.9     .16       0  5092.4     .05       0
Bank Sta=4956,5090.6
XS Rating Curve= 0 ,0
Exp/Cntr=0.3,0.1

Type RM Length L Ch R = 1 ,300881  ,463,463,463
BEGIN DESCRIPTION:
TEHUACANA CREEK 236.0
END DESCRIPTION:
XS GIS Cut Line= 3
      3484499.57     10619310.19      3485949.61     10619410.19
      3486349.61     10619460.19
#Sta/Elev= 30
  3562.1  494.19  3602.2  490.44  3702.5  488.81  4217.4  486.13  4313.9  482.67
  4374.1  482.88  4444.2  479.73  4503.1  480.21    4656  477.56  4845.2  478.13
  4921.7  473.42  4935.4  472.87  4941.7  470.65  4946.7  474.32  4965.5  469.81
  4975.5  469.24  4985.5  463.92  4992.5  463.85  4995.3  463.35  4998.5  463.85
  5018.1  465.84  5035.7  471.31  5053.4  472.47    5066  476.74  5096.2  475.66
    5134  480.43    5197  485.49  5277.6  488.44  5307.8  492.16  5418.7  499.52
#Mann= 5 ,-1 , 0
  3562.1     .05       0  4921.7     .16       0  4992.5     .07       0
  4998.5     .16       0    5134     .05       0
Bank Sta=4845.2,5066
XS Rating Curve= 0 ,0
Exp/Cntr=0.3,0.1

Type RM Length L Ch R = 1 ,300418  ,616,616,616
BEGIN DESCRIPTION:
TEHUACANA CREEK 235.0
END DESCRIPTION:
XS GIS Cut Line= 2
      3485157.91      10619494.1      3486205.32      10619984.2
#Sta/Elev= 30
  4447.9  485.12  4521.4   484.5  4544.2  482.05    4738  475.76  4846.7  474.88
  4891.4  473.45  4920.7  474.69  4943.3  474.29  4971.9  473.87  4979.7  468.12
  4998.8  462.27  5001.6  461.77  5004.8  462.27    5012  464.66  5017.6  472.81
  5023.9  474.79    5046  473.68  5092.8  473.92  5200.3  478.12  5297.1  479.83
  5365.7  479.31  5410.3  482.35  5485.4  485.35  5508.2  485.78  5536.6  484.63
  5559.4  486.91  5564.9  486.53  5582.2  489.44  5587.8  489.01  5604.3  490.65
#Mann= 5 ,-1 , 0
  4447.9     .05       0  4943.3     .16       0  4998.8     .07       0
  5004.8     .16       0  5092.8     .05       0
Bank Sta=4920.7,5023.9
XS Rating Curve= 0 ,0
Exp/Cntr=0.3,0.1

Type RM Length L Ch R = 1 ,299802  ,608,608,608
BEGIN DESCRIPTION:
TEHUACANA CREEK 233.0
END DESCRIPTION:
XS GIS Cut Line= 3
      3484167.02      10620099.9      3485526.39     10620235.31
      3486140.93     10620115.53
#Sta/Elev= 30
  3807.2  490.47  4064.2  487.97  4272.1  484.83  4322.3  485.31    4467  484.16
  4553.5  481.32    4769  483.56  4898.8  479.77  4955.4  476.81  4970.4  475.23
  4975.5  472.81  4985.6  463.13  4992.6  459.07  4995.4  458.57  4998.6  459.07
  5005.7   461.6  5015.7  469.25  5025.8  470.61  5045.9  471.95  5104.8  471.21
  5146.4  471.11  5186.8  473.45    5360  475.11  5379.1  476.11  5390.5  475.08
  5410.9  476.23  5553.5  477.86  5745.5   483.8  5767.5  483.31  5799.4  484.68
#Mann= 5 ,-1 , 0
  3807.2     .05       0  4898.8     .16       0  4992.6     .07       0
  4998.6     .16       0  5104.8     .05       0
Bank Sta=4970.4,5186.8
XS Rating Curve= 0 ,0
Exp/Cntr=0.3,0.1

Type RM Length L Ch R = 1 ,299194  ,928,928,928
BEGIN DESCRIPTION:
TEHUACANA CREEK 232.0
END DESCRIPTION:
XS GIS Cut Line= 2
      3484380.54     10621079.07      3485853.22     10620454.61
#Sta/Elev= 30
  3992.1  495.32  4144.1  489.91  4253.4  490.41  4332.6  488.56  4362.7  487.85
    4472  486.81  4587.1  484.18  4805.7  474.22  4945.7  472.77  4968.7  466.64
  4974.8  462.55  4980.2  465.29  4998.4  458.06  5033.8  471.27  5044.7  471.45
  5102.9  469.37  5120.7  466.25  5127.6  463.73  5133.1   458.1  5139.4  457.98
  5142.2  457.48  5145.4  457.98  5156.7  460.27  5164.2  470.22  5180.4  471.68
  5196.8   479.3  5236.1  472.34  5242.9  471.03  5338.7   467.8  5591.7  478.43
#Mann= 11 ,-1 , 0
  3992.1     .16       0  4144.1      .1       0  4253.4     .05       0
  4332.6      .1       0  4362.7     .05       0    4472     .16       0
  5102.9     .05       0  5139.4     .07       0  5145.4     .05       0
  5236.1     .16       0  5242.9     .05       0
Bank Sta=4945.7,5044.7
XS Rating Curve= 0 ,0
Exp/Cntr=0.3,0.1

Type RM Length L Ch R = 1 ,298266  ,533,533,533
BEGIN DESCRIPTION:
TEHUACANA CREEK 230.0
END DESCRIPTION:
XS GIS Cut Line= 2
      3485259.43     10621769.82      3486311.46     10620391.42
#Sta/Elev= 30
  4148.3  487.34  4519.2  488.51  4633.5  483.16  4639.8  481.86  4697.9  479.79
  4704.2  478.37    4804  473.31  4862.1  471.57    4912  471.57  4946.7  470.25
  4982.7  467.05  4990.7  457.67  4994.2   455.9    4997   455.4  5000.2   455.9
  5003.5   456.3  5011.7  461.79  5026.3  464.63  5032.6  464.79  5040.8  467.41
  5082.4  467.67    5126  469.58  5146.7  468.94  5204.5  469.67    5390  475.36
  5460.7  472.74  5489.7  473.31    5575  472.05  5745.5  474.07  5882.3  478.08
#Mann= 4 ,-1 , 0
  4148.3     .16       0  4994.2     .07       0  5000.2     .16       0
  5146.7     .05       0
Bank Sta=4912,5126
XS Rating Curve= 0 ,0
Exp/Cntr=0.3,0.1

Type RM Length L Ch R = 1 ,297733  ,482,482,482
BEGIN DESCRIPTION:
TEHUACANA CREEK 229.0
END DESCRIPTION:
XS GIS Cut Line= 2
      3486210.79     10621960.85       3486360.1     10620415.65
#Sta/Elev= 30
  4201.5  479.12  4252.4  479.29  4346.5  476.27    4551  473.09  4925.5  470.33
  4955.7  469.23  4966.6  467.78  4975.8   467.2  4985.8  455.21  4992.8  452.72
  4995.6  452.22  4998.8  452.72  5005.9  453.63  5015.9  458.18    5026  464.19
  5059.7  466.36  5086.3  467.92  5196.8  467.42  5226.9  469.38    5237  469.38
  5257.1  467.55  5327.4  467.53  5347.5  468.64  5407.8   468.8    5468  468.06
  5478.1  468.29    5486  469.74    5491  469.22  5628.8  472.77  5753.9  477.59
#Mann= 5 ,-1 , 0
  4201.5     .05       0  4966.6     .16       0  4992.8     .07       0
  4998.8     .16       0  5059.7     .05       0
Bank Sta=4925.5,5086.3
XS Rating Curve= 0 ,0
Exp/Cntr=0.3,0.1

Type RM Length L Ch R = 1 ,297251  ,495,495,495
BEGIN DESCRIPTION:
TEHUACANA CREEK 228.0
END DESCRIPTION:
XS GIS Cut Line= 3
      3486564.96     10621867.04      3486599.61     10620910.19
      3486699.62     10620310.14
#Sta/Elev= 30
  4042.5  476.44  4539.7  470.88  4729.8  467.42  4883.9  468.44  4889.9  468.54
  4939.9  467.42  4959.9  465.46    4970  462.78    4980  461.81    4990  458.05
  4997.5  452.41  5007.1  451.86  5009.9  451.36  5013.1  451.86  5027.9  465.58
  5081.1  464.95  5088.7  460.47  5101.4  460.67  5121.6  464.64  5149.5  463.25
  5154.6  465.63  5162.2  466.01  5253.4  467.73    5294  471.64  5354.8  474.93
  5425.8  476.07    5446  478.06  5466.3  481.76  5527.1  487.37  5608.3  491.29
#Mann= 4 ,-1 , 0
  4042.5     .05       0  4883.9     .16       0  5007.1     .07       0
  5013.1     .16       0
Bank Sta=4889.9,5027.9
XS Rating Curve= 0 ,0
Exp/Cntr=0.3,0.1

Type RM Length L Ch R = 1 ,296756  ,398,398,398
BEGIN DESCRIPTION:
TEHUACANA CREEK 227.0
END DESCRIPTION:
XS GIS Cut Line= 2
      3486730.76      10621943.9      3487043.25     10620147.07
#Sta/Elev= 30
    3756  475.49  4422.5  466.19  4551.5  465.44  4680.3  466.67  4896.6  464.15
  4949.1  464.79  4957.5  461.75  4967.6  460.64  4977.8  453.57  4995.1  450.78
  4997.8  450.28  5001.1  450.78  5003.6  458.23  5018.4  464.96  5058.2  469.09
  5063.2  467.51  5069.1  469.62  5109.7  472.04  5117.8  471.52    5130  473.84
  5160.5  474.78  5174.6  477.25  5237.1  480.09  5272.1  479.34  5282.3  477.91
  5291.6  478.34  5312.7  483.14    5333  482.83  5383.8  486.21  5579.8  489.49
#Mann= 5 ,-1 , 0
    3756     .05       0  4680.3     .16       0  4995.1     .07       0
  5001.1     .16       0  5174.6     .05       0
Bank Sta=4949.1,5069.1
XS Rating Curve= 0 ,0
Exp/Cntr=0.3,0.1

Type RM Length L Ch R = 1 ,296358  ,532,532,532
BEGIN DESCRIPTION:
TEHUACANA CREEK 226.0
END DESCRIPTION:
XS GIS Cut Line= 3
      3486928.69     10621912.62      3487163.05      10621001.2
      3487777.61     10620402.27
#Sta/Elev= 30
  3967.2  478.61  4000.7  475.14  4217.5  471.05  4441.8  463.97  4506.6   460.4
  4553.1  465.64  4764.8  462.75  4963.1  463.61  4977.2  462.56  4984.4  457.94
  4991.4  450.66  4995.5  449.76  4998.3  449.26  5001.5  449.76  5012.7  453.25
  5019.7  463.49  5026.8  467.27  5062.1   468.5    5103  468.57    5253   470.3
  5408.6  473.76    5444  476.12  5465.2  474.65  5493.4  476.22  5500.6  479.16
  5521.7  482.05  5543.1  478.78  5564.2  478.43  5627.9  484.83  5766.4  493.13
#Mann= 5 ,-1 , 0
  3967.2     .05       0  4441.8     .16       0  4995.5     .07       0
  5001.5     .16       0    5103     .05       0
Bank Sta=4963.1,5062.1
XS Rating Curve= 0 ,0
Exp/Cntr=0.3,0.1

Type RM Length L Ch R = 1 ,295826  ,365,365,365
BEGIN DESCRIPTION:
TEHUACANA CREEK 225.0
END DESCRIPTION:
XS GIS Cut Line= 3
      3487038.05     10621943.91       3487256.8     10621480.36
      3488032.83     10620600.17
#Sta/Elev= 30
  4433.8  478.74    4460  479.13  4479.4   476.2  4497.4  474.24  4564.2   473.2
  4871.8  465.45  4955.7  464.36  4969.9  459.45  4976.6  449.68  4981.2  447.96
  4983.9  447.46  4987.2  447.96  4998.4  448.45  5005.1  452.71  5012.6  459.74
  5054.4  462.99  5111.3   463.8  5184.3  465.25  5642.6  472.46  5678.6  474.01
  5699.5  476.53  5713.7  475.46  5742.1  477.05  5748.8  479.63  5784.8   483.1
  5897.7  490.22  5933.1  491.37  5983.1  495.86  6075.1  498.77  6119.8  497.94
#Mann= 7 ,-1 , 0
  4433.8     .05       0  4479.4     .16       0  4564.2     .05       0
  4871.8     .16       0  4981.2     .07       0  4987.2     .16       0
  5184.3     .05       0
Bank Sta=4955.7,5111.3
XS Rating Curve= 0 ,0
Exp/Cntr=0.3,0.1

Type RM Length L Ch R = 1 ,295461  ,468,468,468
BEGIN DESCRIPTION:
TEHUACANA CREEK 224.0
END DESCRIPTION:
XS GIS Cut Line= 2
      3487183.86     10621996.02      3488229.74     10620794.04
#Sta/Elev= 30
  4382.5  474.82  4614.2   468.7  4737.8  462.67    4809  463.64  4858.4  460.27
  4929.6  460.77  4943.8  459.84  4950.4  456.57  4972.3  458.46  4978.9  451.14
  4986.6   452.5  4990.2  447.71  4992.9  447.21  4996.2  447.71    5021  449.55
  5028.3  454.62  5035.9  457.07  5042.5  464.14  5050.2  462.56  5056.8  464.34
    5071  464.53  5156.5  464.15  5318.8  466.38  5361.6  467.48  5383.4  469.79
  5397.7  468.11  5666.4  482.43  5815.4  492.26  5893.3  494.21  5975.8  493.44
#Mann= 5 ,-1 , 0
  4382.5     .05       0  4614.2     .16       0  4990.2     .07       0
  4996.2     .16       0    5021     .05       0
Bank Sta=4929.6,5071
XS Rating Curve= 0 ,0
Exp/Cntr=0.3,0.1

Type RM Length L Ch R = 1 ,294993  ,534,534,534
BEGIN DESCRIPTION:
TEHUACANA CREEK 223.0
END DESCRIPTION:
XS GIS Cut Line= 3
      3487168.27     10622079.32      3487668.26     10621995.99
      3488344.96     10620960.13
#Sta/Elev= 30
  4412.5  474.44  4444.3  475.01  4464.6  473.75  4535.5  473.58  4636.9  468.64
  4728.1  465.74  4902.4  463.57  4967.8  463.83  4974.1  457.48    4983  453.99
  4988.9  448.66    4995  445.05  4997.7  444.55    5001  445.05  5004.1  445.06
  5019.2  450.87  5025.1  458.35  5040.3  460.63  5061.3  461.52  5217.1  462.85
  5320.7   464.2  5429.3  463.11  5640.6  466.93  5654.9  467.56  5667.6   470.1
  5682.7  469.32  5762.5  473.76  5957.2  488.63  6065.8  492.07  6156.7  491.57
#Mann= 5 ,-1 , 0
  4412.5     .05       0  4902.4     .16       0    4995     .07       0
    5001     .16       0  5217.1     .05       0
Bank Sta=4967.8,5061.3
XS Rating Curve= 0 ,0
Exp/Cntr=0.3,0.1

Type RM Length L Ch R = 1 ,294459  ,556,556,556
BEGIN DESCRIPTION:
TEHUACANA CREEK 222.0
END DESCRIPTION:
XS GIS Cut Line= 4
      3488365.62     10622807.72      3488080.86     10621848.49
      3488132.95     10621660.99      3488361.38     10621193.74
#Sta/Elev= 30
  3888.7  467.99  4470.3  463.83  4592.6  460.69  4678.9  462.17  4795.5  459.39
  4866.7  458.85  4889.3  454.34  4908.4  455.49  4929.1  460.26  4937.5  460.15
  4960.2     459  4970.6  457.02  4991.3  444.53  4998.7  443.77  5001.5  443.27
  5004.7  443.77  5016.3  445.24  5022.5  449.64  5032.8  461.65  5033.4  461.63
  5055.8  460.84  5081.7  462.31  5201.6  463.57  5246.6  466.38  5307.4  468.31
  5314.2  469.76  5329.7  469.02  5409.8  474.01  5463.3  479.99    5604  488.52
#Mann= 5 ,-1 , 0
  3888.7     .05       0  4795.5     .16       0  4998.7     .07       0
  5004.7     .16       0  5033.4     .05       0
Bank Sta=4937.5,5032.8
XS Rating Curve= 0 ,0
Exp/Cntr=0.3,0.1

Type RM Length L Ch R = 1 ,293903  ,490,490,490
BEGIN DESCRIPTION:
TEHUACANA CREEK 221.0
END DESCRIPTION:
XS GIS Cut Line= 4
      3488498.42     10622989.97      3488519.55     10621932.26
       3488539.2     10621827.65      3488632.76     10621203.89
#Sta/Elev= 30
  3891.7   468.7  4221.5  467.07  4291.6  464.61  4513.1  461.06  4651.6   457.4
  4691.6  459.21  4921.7  457.38  4948.2  458.59  4977.1  455.58  4982.3  448.92
  4992.4  442.79  4999.6  442.77  5002.4  442.27  5005.6  442.77  5012.8  445.09
  5022.9  456.65  5029.6  459.87  5037.3  461.37  5043.3  461.47  5144.5   460.7
  5377.1  463.84    5458  467.14  5508.5  467.29  5518.6  469.39  5564.3  471.69
  5569.3  470.65  5579.3  472.25  5599.5  471.48    5640  475.15  5686.8  476.92
#Mann= 5 ,-1 , 0
  3891.7     .05       0  4513.1     .16       0  4999.6     .07       0
  5005.6     .16       0  5037.3     .05       0
Bank Sta=4948.2,5043.3
XS Rating Curve= 0 ,0
Exp/Cntr=0.3,0.1

Type RM Length L Ch R = 1 ,293413  ,545,545,545
BEGIN DESCRIPTION:
TEHUACANA CREEK 220.0
END DESCRIPTION:
XS GIS Cut Line= 3
      3488679.82     10622634.96      3488898.57     10622140.15
      3488919.41      10621249.5
#Sta/Elev= 30
    4537  466.82    4577  466.99  4706.2  464.54    4739  463.06  4751.1   464.2
  4792.2  464.63  4797.7  463.21    4821  461.77    4873  462.92  4925.1  461.24
  4957.7  455.57  4979.6  452.96  4989.5  447.14    4995  440.81  4998.4  440.73
  5001.2  440.23  5004.4  440.73  5012.4  442.76  5018.3  451.28  5023.8  456.18
  5047.1  457.99    5108  456.19  5161.9  458.17    5198  459.31    5308  459.93
  5558.1  459.18  5768.5  461.81  5908.2  465.82  5948.2  465.96  5968.9  467.58
#Mann= 4 ,-1 , 0
    4537     .16       0  4998.4     .07       0  5004.4     .16       0
  5161.9     .05       0
Bank Sta=4925.1,5047.1
XS Rating Curve= 0 ,0
Exp/Cntr=0.3,0.1

Type RM Length L Ch R = 1 ,292868  ,68,68,68
BEGIN DESCRIPTION:
TEHUACANA CREEK 219.0
END DESCRIPTION:
XS GIS Cut Line= 4
      3489243.21     10623409.26      3489292.67     10622266.89
      3489287.46     10622063.76      3489318.71     10620996.05
#Sta/Elev= 30
  3810.5  470.46  3837.4  470.01  4049.8  462.57  4099.8  463.44  4138.5  467.04
  4420.1  464.76  4460.2   460.4  4523.4  464.22  4580.3  465.61  4690.4  462.05
  4766.5  462.36  4800.5  459.64  4830.5   456.6  4860.6  449.69  4880.6  448.13
  4920.6  455.12  4930.6  453.83  4949.8  443.85  4980.6  443.61  4997.7  438.97
  5000.4  438.47  5003.7  438.97  5060.7  448.28  5070.7   450.6  5080.7  458.09
  5090.7  458.47  5114.8  457.73    5931  461.08  6161.1  464.66  6225.3  467.47
#Mann= 7 ,-1 , 0
  3810.5     .05       0  3837.4     .16       0  4138.5     .05       0
  4523.4     .16       0  4997.7     .07       0  5003.7     .16       0
  5114.8     .05       0
Bank Sta=4800.5,5090.7
XS Rating Curve= 0 ,0
Exp/Cntr=0.3,0.1

Type RM Length L Ch R = 1 ,292800  ,908,908,908
BEGIN DESCRIPTION:
TEHUACANA CREEK 218.0
END DESCRIPTION:
XS GIS Cut Line= 6
      3489329.15     10623380.62      3489346.49     10622645.36
      3489346.49     10622369.32      3489372.53     10621957.86
      3489372.53     10621718.28      3489403.75     10620984.57
#Sta/Elev= 30
  3851.3  469.59  3921.7  469.08  4001.8  464.81  4211.8  466.96  4341.9  464.53
  4461.9  459.95    4507  462.53  4532.2  460.44  4561.9  462.85  4630.2  462.49
  4741.9  460.23  4761.9  458.43  4821.9  459.06    4882  454.19  4952.2  453.52
  4972.3  450.11  4992.4   440.2  4999.4  438.85  5002.1  438.35  5005.4  438.85
  5022.5  454.57  5042.5  454.09  5051.8  457.93  5062.6  458.69  5382.8   456.6
  5502.8  458.49  5632.9  457.11  5923.2  459.49  6153.4  465.46  6249.1  472.81
#Mann= 5 ,-1 , 0
  3851.3     .05       0  4532.2     .08       0  4630.2     .05       0
  4999.4     .04       0  5005.4     .05       0
Bank Sta=4821.9,5062.6
XS Rating Curve= 0 ,0
Exp/Cntr=0.3,0.1

Type RM Length L Ch R = 1 ,291892  ,1455,1455,1455
BEGIN DESCRIPTION:
TEHUACANA CREEK 217.0
END DESCRIPTION:
XS GIS Cut Line= 4
      3490099.98     10623216.54      3490166.34     10622369.53
      3489558.71      10621557.9      3489576.07     10620976.35
#Sta/Elev= 30
  3787.5  467.18  3934.3  464.58  4034.6  464.68  4074.7  467.04  4106.3  463.27
  4144.9  462.35  4846.7  456.39  4941.3   456.6  4962.2  455.47  4970.5  445.99
  4985.1  439.48  4995.6  437.93  4998.3  437.43  5001.6  437.93  5005.9  438.01
  5012.2  445.65  5026.8  452.13  5062.4  453.37  5241.4  456.38  5398.3  454.27
  5541.5  456.85  5738.7  455.81  5851.3  456.72  5988.9  459.16  6008.9   460.8
  6018.9  460.06  6138.9  464.26  6178.9  466.87    6184  468.58  6232.8  471.07
#Mann= 5 ,-1 , 0
  3787.5     .05       0  4846.7     .16       0  4995.6     .07       0
  5001.6     .16       0  5062.4     .05       0
Bank Sta=4941.3,5241.4
XS Rating Curve= 0 ,0
Exp/Cntr=0.3,0.1

Type RM Length L Ch R = 1 ,290437  ,1093,1093,1093
BEGIN DESCRIPTION:
TEHUACANA CREEK 216.0
END DESCRIPTION:
XS GIS Cut Line= 2
      3490422.06     10623014.59      3490547.93     10620779.33
#Sta/Elev= 30
  3443.2  462.25  3998.1  457.82  4119.1  457.85    4303  456.42    4597  455.39
    4695  455.64  4769.7   454.8  4919.9  452.56    4940  451.73    4950  448.58
    4960  450.98    4970  449.04    4980  444.92    4990  436.38  4997.1  435.58
  4999.8  435.08  5003.1  435.58  5020.1  437.09  5030.1  445.43  5035.1  446.73
  5070.2  451.07  5080.2  451.02  5092.3   447.7  5100.2  450.05  5140.3  453.08
  5200.4  455.24  5320.6  460.44  5390.7  466.58  5520.9  472.89    5682  475.81
#Mann= 9 ,-1 , 0
  3443.2     .05       0  3998.1     .16       0  4119.1     .05       0
    4303     .16       0    4597     .05       0    4695     .16       0
  4997.1     .07       0  5003.1     .16       0  5035.1     .05       0
Bank Sta=4769.7,5200.4
XS Rating Curve= 0 ,0
Exp/Cntr=0.3,0.1

Type RM Length L Ch R = 1 ,289344  ,526,526,526
BEGIN DESCRIPTION:
TEHUACANA CREEK 215.0
END DESCRIPTION:
XS GIS Cut Line= 3
       3490799.6     10623610.21      3491199.61     10621210.19
       3491299.6     10620810.23
#Sta/Elev= 30
  2561.5  468.27  3058.3  465.03  3420.2  456.42  3524.6  453.96  3544.9  456.29
  3727.4  455.07  3861.5  451.78  3879.5  451.51  3889.6  448.76  3899.7  451.84
  3909.9  452.05  4012.8  451.14  4111.6  449.98  4115.2  449.08  4132.9  453.27
  4236.8   450.9  4557.9  453.06  4771.6   448.6  4883.1  450.64  4979.3   446.6
  4984.5  445.98  4992.1  435.89  5001.9  435.26  5004.7  434.76  5007.9  435.26
  5012.7  437.55  5017.8  436.56  5035.9  453.61  5200.8  456.91  5406.9  468.73
#Mann= 9 ,-1 , 0
  2561.5     .05       0  3420.2     .16       0  3861.5     .05       0
  4012.8     .16       0  4111.6     .05       0  4557.9     .16       0
  4979.3     .05       0  5001.9    .035       0  5007.9     .05       0
Bank Sta=4883.1,5035.9
XS Rating Curve= 0 ,0
Exp/Cntr=0.3,0.1

Type RM Length L Ch R = 1 ,288818  ,535,535,535
BEGIN DESCRIPTION:
TEHUACANA CREEK 214.0
END DESCRIPTION:
XS GIS Cut Line= 3
      3491449.61     10623310.16      3491449.61     10621510.19
      3491349.61     10620510.15
#Sta/Elev= 30
  3191.8  470.65  3281.8  465.39  3581.8  464.88  3811.8  459.82  4503.8  450.54
    4508  450.59  4561.8  448.41  4571.8  449.75  4631.8  448.75  4641.8  446.57
  4691.8  447.63  4731.8  443.64  4751.8  444.12  4781.8   449.3  4931.8  451.15
  4961.8  450.55  4971.8   447.6  4989.3  436.98  5008.9  435.37  5011.6  434.87
  5014.9  435.37  5021.9  440.12  5039.5  446.08  5082.2  448.31  5263.1  451.39
  5423.9  459.24    5635  467.16  5665.1  466.75  5715.4  470.77  5996.8   479.9
#Mann= 5 ,-1 , 0
  3191.8     .05       0  4503.8     .16       0    4508     .05       0
  5008.9    .035       0  5014.9     .05       0
Bank Sta=4931.8,5263.1
XS Rating Curve= 0 ,0
Exp/Cntr=0.3,0.1
