HEC-RAS study TEHUACANA CREEK.prj: TEHUACANA CREEK Base Level Engineering

--- TEHUACANA CREEK.g01 (geometry) --- (continued)

Type RM Length L Ch R = 1 ,85492   ,1574,1574,1574
BEGIN DESCRIPTION:
TEHUACANA CREEK 33.0
END DESCRIPTION:
XS GIS Cut Line= 3
      3595566.44     10685076.27      3598886.74     10682797.62
      3599255.67     10679629.22
#Sta/Elev= 30
  2339.8  325.83  3194.3  299.42    3310   289.5  3489.9  274.82  3548.5  270.52
  3684.3  262.18  4329.1  260.64  4373.1  260.97  4434.4  258.38  4963.4  263.97
  4993.2  248.07    5020  247.88  5022.7  247.38    5026  247.88  5064.9  263.42
  5069.2  262.98  5290.4  260.53  5439.2   260.9  6538.3  262.31  6794.4  263.29
  6864.8   263.8  6887.7  255.04  7136.9  263.01  7333.4  266.87  7431.6  269.71
  7686.7   273.1  8312.2  274.74  8774.7  276.88  9032.9  278.26  9556.6  319.36
#Mann= 20 ,-1 , 0
  2339.8     .16       0    3310     .12       0  3489.9     .16       0
  3548.5     .12       0  4329.1     .07       0  4373.1     .16       0
  4434.4     .12       0    5020     .07       0    5026     .12       0
  5069.2     .07       0  5290.4     .05       0  5439.2     .12       0
  6538.3     .05       0  6794.4     .12       0  7136.9     .12       0
  7333.4     .16       0  7431.6     .05       0  7686.7      .1       0
  8312.2     .05       0  8774.7     .16       0
Bank Sta=4963.4,5064.9
XS Rating Curve= 0 ,0
Exp/Cntr=0.3,0.1

Type RM Length L Ch R = 1 ,83918   ,2196,2196,2196
BEGIN DESCRIPTION:
TEHUACANA CREEK 32.0
END DESCRIPTION:
XS GIS Cut Line= 4
      3598821.64      10687521.3      3598865.04     10684700.11
      3599971.81     10682508.27      3601773.01     10680229.65
#Sta/Elev= 30
  1859.5   321.9  1938.3  320.05  2759.8  287.27  3072.6  287.88  3155.3  285.22
  3346.6  273.56  3501.1  267.58  3740.8   263.9  3770.8   252.6  3800.8  263.32
  4945.2  263.72  4980.4   248.3  4983.2   247.8  4986.4   248.3  5034.4  249.78
  5048.2  261.27    5079  263.88  6661.2  262.65    6701  254.17  6780.9   263.5
  7197.2   261.8  7847.9  266.45  8015.4  284.05  8152.1  295.54  8875.3  303.56
  9256.8  307.45  9373.4  309.43  9494.6  311.49    9651  314.14   10041     317
#Mann= 20 ,-1 , 0
  1859.5     .05       0  1938.3     .16       0  2759.8     .12       0
  3072.6     .16       0  3155.3     .12       0  3346.6     .16       0
  3501.1     .12       0  4980.4     .07       0  4986.4     .16       0
  5048.2     .12       0  6661.2     .07       0  6780.9     .05       0
  7197.2     .05       0  7847.9     .16       0  8015.4     .05       0
  8875.3     .16       0  9256.8     .12       0  9373.4     .16       0
  9494.6     .12       0    9651     .16       0
Bank Sta=4945.2,5079
XS Rating Curve= 0 ,0
Exp/Cntr=0.3,0.1

Type RM Length L Ch R = 1 ,81722   ,1635,1635,1635
BEGIN DESCRIPTION:
TEHUACANA CREEK 31.0
END DESCRIPTION:
XS GIS Cut Line= 2
      3600275.64     10687456.18      3602336.78     10680643.55
#Sta/Elev= 30
  2546.9  312.73    2830  302.81    3056  299.91  3437.4  293.63  3725.2  284.66
  3765.1  274.14  4044.8  257.86  4146.1  259.25  4253.6  258.64  4914.3  263.94
    4958  247.25  4960.7  246.75    4964  247.25  4999.1  248.32  5039.7  263.59
    5157  259.44  5259.7  259.35  5360.9  258.66  5462.1  258.37  5563.4  258.39
    6272  258.76  6575.7  260.03  6615.1  260.35  6627.7  251.06    6708  260.39
  7923.3  267.45  8827.6  306.23  9362.9   315.3  9647.8  317.07  9664.5  316.62
#Mann= 20 ,-1 , 0
  2546.9     .05       0    2830     .16       0    3056     .05       0
  3437.4     .08       0  3725.2     .05       0  4044.8     .16       0
  4146.1     .05       0  4253.6     .16       0    4958     .03       0
    4964     .05       0    5157     .05       0  5259.7     .07       0
  5360.9     .12       0  5462.1     .07       0  5563.4     .12       0
    6272     .05       0  6575.7     .07       0    6708     .05       0
  9362.9     .16       0  9647.8     .05       0
Bank Sta=4914.3,5039.7
XS Rating Curve= 0 ,0
Exp/Cntr=0.3,0.1

Type RM Length L Ch R = 1 ,80087   ,1601,1601,1601
BEGIN DESCRIPTION:
Mapping XS 0550fcb2
END DESCRIPTION:
XS GIS Cut Line= 3
      3601208.82     10687586.36      3602424.07     10685654.97
      3603552.54      10681141.1
#Sta/Elev= 30
  2158.2  318.27  2243.2  312.23  2379.8   301.8  2469.3   297.4  3034.6  264.22
  3154.1   259.2  3368.8  257.85  3504.8  257.52  3623.8   257.7  3944.7  257.53
  4163.2  258.27  4278.2  257.32  4391.2  258.42  4897.2  261.13    4941  261.59
    5009  247.08  5011.7  246.58    5015  247.08  5064.7  262.19  5415.8  257.73
  6498.6  258.14  6798.8  256.84  6832.5  250.15  6857.1  259.93  6898.9  259.71
    7558  259.65  8104.3  278.39  8578.5  313.02  8722.8  317.73  9092.9  312.78
#Mann= 20 ,-1 , 0
  2158.2     .16       0  2243.2     .16       0  2379.8     .05       0
  2469.3     .16       0  3034.6     .12       0  3154.1     .07       0
  3368.8     .12       0  3504.8     .07       0  3623.8     .12       0
  3944.7     .05       0  4163.2     .07       0  4278.2     .05       0
  4391.2     .07       0  4897.2     .05       0    5009     .07       0
    5015     .12       0  5415.8     .05       0  6498.6     .07       0
  6798.8     .12       0  6898.9     .05       0
Bank Sta=4941,5064.7
XS Rating Curve= 0 ,0
Exp/Cntr=0.3,0.1

Type RM Length L Ch R = 1 ,78486   ,5421,5421,5421
BEGIN DESCRIPTION:
Mapping XS b74d5d6e
END DESCRIPTION:
XS GIS Cut Line= 4
      3601447.51      10687694.9      3603791.26      10686132.4
      3604615.91     10684005.67      3604030.21     10681424.23
#Sta/Elev= 30
  1805.2  307.63  2433.5  301.75  2632.5  296.84  3122.2  263.18  3268.3  261.42
  3658.7  260.58    3936  260.28  3962.3  259.97  4269.9  257.89  4315.6  257.58
  4938.2  261.66  4956.3  251.66  4999.8  247.37  5017.2  259.01  5053.4  261.43
  5266.3  257.39  5359.8  256.76  5398.9  254.82  6164.5  257.44  6268.1  257.69
  6371.7  257.94  6468.3  254.27  6487.6  246.26  6490.4  245.76  6493.6  246.26
  6501.4  255.37  6522.8  258.07  8266.1  257.54  9217.4  314.31  9550.1  301.38
#Mann= 18 ,-1 , 0
  1805.2     .05       0  2433.5     .16       0  3268.3     .12       0
  3658.7     .16       0    3936     .12       0  3962.3     .16       0
  4269.9     .12       0  4315.6     .05       0  4956.3     .12       0
  5266.3     .05       0  5359.8     .12       0  5398.9     .05       0
  6164.5     .07       0  6268.1     .05       0  6371.7     .12       0
  6468.3     .05       0  6487.6     .07       0  6493.6     .05       0
Bank Sta=4938.2,5053.4
XS Rating Curve= 0 ,0
Exp/Cntr=0.3,0.1

Type RM Length L Ch R = 1 ,73065   ,381,381,381
BEGIN DESCRIPTION:
Mapping XS d6cf8573
END DESCRIPTION:
XS GIS Cut Line= 3
      3605883.49     10688104.66      3605466.82     10684042.12
      3604598.77     10680535.21
#Sta/Elev= 30
   419.9  296.11   598.6  288.85    1108  267.83  1495.4  265.05  1679.5  262.77
  2394.7   260.5  2434.9  247.71  2485.1   260.7  3311.8  256.37  3603.5  254.99
  3801.4  257.34  3999.3  257.55  4098.3  257.47  4157.3  257.05  4197.2  256.98
    4213  256.95  4494.1  255.92  4759.9  256.54  4931.2   257.9  5005.9  243.12
  5008.6  242.62  5011.9  243.12  5041.4   243.7  5055.4  256.03    5927  263.74
  6227.7   266.6  7305.5  278.64  7307.1  278.54  7674.8  297.88  8116.5  308.13
#Mann= 20 ,-1 , 0
   419.9     .05       0   598.6     .12       0  1495.4     .16       0
  1679.5     .12       0  3311.8     .07       0  3603.5     .12       0
  3801.4     .07       0  3999.3     .05       0  4098.3     .07       0
  4157.3     .05       0  4197.2     .07       0    4213     .05       0
  4494.1     .07       0  4759.9     .05       0  5005.9     .03       0
  5011.9     .05       0    5927     .16       0  6227.7     .05       0
  7305.5     .16       0  7307.1     .05       0
#XS Ineff= 1 ,-1
 2394.49 2483.55  260.34
Permanent Ineff=
       F
Bank Sta=4931.2,5055.4
XS Rating Curve= 0 ,0
Exp/Cntr=0.3,0.1

Type RM Length L Ch R = 1 ,72684   ,212,212,212
BEGIN DESCRIPTION:
Mapping XS b20a86de
END DESCRIPTION:
XS GIS Cut Line= 2
      3606925.16     10687826.88      3604928.61     10680778.19
#Sta/Elev= 30
   339.4  313.11   743.6  307.66   894.7  301.99  1213.7  288.08  1464.9  284.15
  1877.1  269.02    2134  256.28  2352.3  259.22  2373.1  247.28  2397.7   258.9
  2598.4   258.3  2701.5  257.19  3765.9  256.53    3938  256.61  4144.1  256.05
  4247.1  255.18  4453.2  255.52  4722.9  255.92  4865.4   255.5  4940.2  256.71
  4992.2   243.3  5051.6   243.2  5054.3   242.7  5057.6   243.2  5077.7  255.44
  5127.3  256.27  5895.8  267.24  5998.9  263.63  6636.9  273.15  7665.4  290.38
#Mann= 20 ,-1 , 0
   339.4     .05       0   743.6     .08       0   894.7     .05       0
  1213.7     .05       0  1464.9     .05       0  1877.1     .12       0
  2598.4     .07       0  2701.5     .05       0  3765.9     .07       0
    3938     .05       0  4144.1     .08       0  4247.1     .05       0
  4453.2     .08       0  4722.9     .05       0  4865.4     .08       0
  5051.6     .07       0  5057.6     .05       0  5895.8     .08       0
  5998.9     .05       0  6636.9     .05       0
#XS Ineff= 1 ,-1
 2345.32 2404.25  258.86
Permanent Ineff=
       F
Bank Sta=4940.2,5127.3
XS Rating Curve= 0 ,0
Exp/Cntr=0.3,0.1

Type RM Length L Ch R = 1 ,72472   ,1509,1509,1509
BEGIN DESCRIPTION:
Mapping XS 15fbb473
END DESCRIPTION:
XS GIS Cut Line= 2
       3606994.6      10687722.7      3605084.86     10680708.75
#Sta/Elev= 30
   342.7  312.37     839  300.29  1147.2  292.22    1899  267.36  2148.7  267.67
  2281.1  247.31  2320.8  258.72  2532.1   254.7  2588.8  266.05  3612.2  260.47
  3714.9  262.01  4125.7  261.78  4331.1  262.43  4466.5  264.54  4722.1  267.02
  4844.7   250.9  4964.7  243.25  4967.4  242.75  4970.7  243.25  5085.3  254.02
  5178.5  268.19  5255.5  264.68  5460.9   263.9  5666.3  260.38  5871.8  262.69
    6488   272.2  6731.9  280.96  6898.9  284.08  7061.2  288.84    7612  301.64
#Mann= 20 ,-1 , 0
   342.7     .05       0     839     .05       0  1147.2     .05       0
  3612.2     .08       0  3714.9     .05       0  4125.7     .08       0
  4331.1     .05       0  4466.5     .08       0  4844.7      .1       0
  4964.7     .07       0  4970.7      .1       0  5085.3     .08       0
  5255.5     .05       0  5460.9     .08       0  5666.3     .05       0
  5871.8     .05       0    6488     .08       0  6731.9     .08       0
  6898.9     .05       0  7061.2     .08       0
#XS Ineff= 1 ,-1
 2149.12 2570.65  265.24
Permanent Ineff=
       F
Bank Sta=4722.1,5178.5
XS Rating Curve= 0 ,0
Exp/Cntr=0.3,0.1

Type RM Length L Ch R = 1 ,70963   ,2256,2256,2256
BEGIN DESCRIPTION:
TEHUACANA CREEK 30.0
END DESCRIPTION:
XS GIS Cut Line= 3
      3607199.61     10687060.16      3607199.61     10683060.19
       3605500.5      10680450.8
#Sta/Elev= 30
   999.8     296  1391.3  280.42  1489.3  274.01  1532.2  269.42  2549.8  258.54
  2579.8  246.81  2709.8  246.46  2739.8  258.58  3078.6  256.77  4423.7  254.75
  4724.8  254.93  4859.8  258.68  4899.8   258.4  4926.8  243.23  4929.5  242.73
  4932.8  243.23  5049.5  246.35  5085.8  257.34  5107.2  256.25  5143.3  257.29
  5372.2  278.57  5503.5  285.52  5620.4  289.34    6989  282.64  7064.3  283.81
    7160  285.05  7729.3  308.86  7918.4  310.95  8015.3  312.93  8113.6  316.64
#Mann= 20 ,-1 , 0
   999.8     .16       0  1391.3     .12       0  1489.3     .16       0
  1532.2     .12       0  3078.6     .05       0  4423.7     .07       0
  4724.8     .05       0  4926.8     .07       0  4932.8     .05       0
  5107.2     .16       0  5143.3     .12       0  5372.2     .05       0
  5503.5     .16       0  5620.4     .05       0    6989     .16       0
  7064.3     .05       0    7160     .16       0  7729.3     .05       0
  7918.4     .16       0  8015.3     .05       0
#XS Ineff= 1 ,-1
 2536.36 2751.14  258.42
Permanent Ineff=
       F
Bank Sta=4859.8,5085.8
XS Rating Curve= 0 ,0
Exp/Cntr=0.3,0.1

Type RM Length L Ch R = 1 ,68707   ,568,568,568
BEGIN DESCRIPTION:
TEHUACANA CREEK 29.0
END DESCRIPTION:
XS GIS Cut Line= 4
      3607857.29     10687501.11      3609576.02     10683673.03
      3609237.48     10682683.44      3605533.85     10679887.16
#Sta/Elev= 30
   208.8  300.86   243.7  301.52   567.3  292.66   895.1     269  1275.9   259.4
  1579.2  256.56  2351.8  256.76  2358.3  247.26  2369.3  245.79  2403.6  256.58
  2450.9  256.24  2582.8  254.48  2873.3  254.06  3093.3  253.31  4969.5  256.33
  5007.5  243.01  5010.2  242.51  5013.5  243.01  5063.4  256.75  7627.5  255.74
  8279.9  273.92  8397.9   271.9  8590.9  285.12  8737.9  289.55  8946.2  295.92
  9046.4   298.3  9292.9  305.77  9621.1  313.09 10036.1  318.45 10091.6  318.93
#Mann= 20 ,-1 , 0
   208.8     .08       0   243.7     .05       0   895.1     .16       0
  1275.9     .12       0  1579.2     .12       0  2450.9     .07       0
  2582.8     .12       0  2873.3     .05       0  3093.3     .05       0
  5007.5     .03       0  5013.5     .05       0  7627.5     .05       0
  8397.9     .16       0  8590.9     .12       0  8737.9     .16       0
  8946.2     .16       0  9046.4     .05       0  9292.9     .16       0
  9621.1     .12       0 10036.1     .05       0
#XS Ineff= 1 ,-1
 2345.64 2412.58  256.56
Permanent Ineff=
       F
Bank Sta=4969.5,5063.4
XS Rating Curve= 0 ,0
Exp/Cntr=0.3,0.1

Type RM Length L Ch R = 1 ,68139   ,1390,1390,1390
BEGIN DESCRIPTION:
TEHUACANA CREEK 28.0
END DESCRIPTION:
XS GIS Cut Line= 3
      3611499.61     10685710.19      3609899.61     10682910.19
       3610699.6     10679310.21
#Sta/Elev= 30
  1805.1  305.71    2427  268.27  2890.6  253.84  2910.8   249.1  3152.6  255.24
  3183.6  245.15    3211  255.64  3695.8  252.67  4349.8  252.96  4796.1   251.3
  4957.3  256.27  4978.6  242.52  5016.3  243.53  5049.2  255.93    5103  255.21
  5515.3  252.56  5984.7  252.55  6474.4  252.54  7700.8  257.14  7771.5  258.17
  7806.1  248.07  7815.1  248.26  7820.2   257.4  7850.5  258.16  7907.3  256.47
  8091.7  270.57  8174.9  280.07  8329.8     310  8492.5  328.55  8717.8  331.04
#Mann= 10 ,-1 , 0
  1805.1     .05       0  2890.6     .16       0  3695.8     .16       0
  4349.8     .16       0    5103     .16       0  5515.3     .16       0
  5984.7     .16       0  6474.4     .16       0  7700.8     .16       0
  7850.5     .05       0
Bank Sta=4957.3,5049.2
XS Rating Curve= 0 ,0
Exp/Cntr=0.3,0.1

Type RM Length L Ch R = 1 ,66749   ,1035,1035,1035
BEGIN DESCRIPTION:
TEHUACANA CREEK 27.0
END DESCRIPTION:
XS GIS Cut Line= 3
      3611549.61     10685660.21      3611149.61     10682460.19
      3610749.61     10679260.22
#Sta/Elev= 30
  1780.5  306.76  2490.8  256.27  2785.8   249.4  3413.1  254.59  3443.4  244.04
  3463.5  254.42  3976.5  251.72  4062.1  252.08  4161.4  251.75  4602.4  252.07
  4624.1  252.13  4922.7  254.74  4967.6  255.34  4992.3  241.67  4995.1  241.17
  4998.3  241.67  5025.6  243.19  5055.1  253.35    5076  254.89    5353  254.19
  5452.3  253.86  6941.7  257.13  7000.8   257.4  7031.1  248.49  7078.8  247.66
  7101.6  258.16  7232.6  256.58  7403.9  269.17  7978.4  334.53  8230.3  336.26
#Mann= 15 ,-1 , 0
  1780.5     .05       0  2490.8     .12       0  3976.5     .12       0
  4062.1     .12       0  4161.4     .12       0  4602.4     .07       0
  4624.1     .12       0  4922.7     .07       0  4992.3     .07       0
  4998.3     .07       0  5055.1     .12       0    5353     .08       0
  5452.3     .12       0  6941.7     .12       0  7078.8     .05       0
#XS Ineff= 1 ,-1
 3411.87 3465.84  254.46
Permanent Ineff=
       F
Bank Sta=4967.6,5076
XS Rating Curve= 0 ,0
Exp/Cntr=0.3,0.1

Type RM Length L Ch R = 1 ,65714   ,2118,2118,2118
BEGIN DESCRIPTION:
TEHUACANA CREEK 26.0
END DESCRIPTION:
XS GIS Cut Line= 2
      3612777.41     10686028.44      3611545.07     10679033.56
#Sta/Elev= 30
    1129  300.78  1340.5   296.5  1958.9  255.89    2156  251.15  2833.8  251.12
  4021.1  254.65  4051.6  243.47  4080.7  254.58  4287.6  251.39  4399.5  251.38
  4410.1  251.05  4822.1  251.76  4955.3   254.9  5000.8  241.68  5003.6  241.18
  5006.8  241.68  5026.4  254.14  5046.7  254.47  5063.1  247.32  5087.3  254.22
  5181.2   253.2  6317.3   254.5  6711.9  256.63  6736.5  246.53  6762.7  256.21
  6909.7  255.79  7219.6  254.84  7778.2  282.71  8005.1   287.8  8231.6  309.49
#Mann= 13 ,-1 , 0
    1129     .05       0  1958.9     .12       0    2156     .05       0
  2833.8     .12       0  4287.6     .05       0  4399.5     .07       0
  4410.1     .05       0  4822.1     .07       0  5000.8     .07       0
  5006.8     .07       0  5181.2     .05       0  6317.3     .16       0
  6909.7     .05       0
#XS Ineff= 1 ,-1
 4027.02 4082.23  253.91
Permanent Ineff=
       F
Bank Sta=4955.3,5046.7
XS Rating Curve= 0 ,0
Exp/Cntr=0.3,0.1

Type RM Length L Ch R = 1 ,63596   ,2216,2216,2216
BEGIN DESCRIPTION:
TEHUACANA CREEK 25.0
END DESCRIPTION:
XS GIS Cut Line= 3
      3613784.35     10685906.85       3613853.8     10681827.02
        3613767.     10679605.04
#Sta/Elev= 30
   616.1  306.54   730.6  297.88   880.2  284.77  1342.9  251.49  1843.5   250.6
  1851.1  250.58  1932.4  250.32    1949  250.27  2635.1  250.82  2733.1  250.84
  2815.1  250.83  4073.3  253.63  4103.3  243.04  4123.3  252.65  4491.7  250.98
  4758.6  252.64  4893.5     253  4903.5  246.42  4953.6  253.75  4955.2  253.72
  4973.6  253.43  4983.6   244.2  5000.6  240.36  5003.3  239.86  5006.6  240.36
  5043.6  253.86  5622.6  250.16  6344.6  249.68  6727.6  289.14  6920.2  291.88
#Mann= 16 ,-1 , 0
   616.1     .05       0   730.6     .16       0   880.2     .05       0
  1843.5     .07       0  1851.1     .05       0  1932.4     .07       0
    1949     .05       0  2635.1     .12       0  2733.1     .07       0
  2815.1     .12       0  4491.7     .05       0  4758.6     .07       0
  4955.2     .05       0  5000.6     .03       0  5006.6     .05       0
  5622.6     .12       0
#XS Ineff= 1 ,-1
  4077.4 4124.17   252.5
Permanent Ineff=
       F
Bank Sta=4953.6,5043.6
XS Rating Curve= 0 ,0
Exp/Cntr=0.3,0.1

Type RM Length L Ch R = 1 ,61380   ,1660,1660,1660
BEGIN DESCRIPTION:
TEHUACANA CREEK 24.0
END DESCRIPTION:
XS GIS Cut Line= 3
      3614201.02     10685993.67      3615555.19     10681184.66
      3615676.72      10678649.9
#Sta/Elev= 30
  -354.1  288.82  -117.1  280.41   332.3   251.8    1645  249.48  2050.7  249.75
  2271.2   249.7  2379.2  249.94  2499.3   249.7  2700.8  249.38  3798.4  250.28
  4269.1  252.31  4308.3  251.45  4335.4  242.12  4376.4  251.98  4605.7   250.2
  4738.1  250.01  4916.7     251  4956.8  250.17  4993.8  239.81  4996.6  239.31
  4999.8  239.81  5036.9  252.39  5105.7  250.66  5314.1  249.96    6018  250.15
  6368.4   282.6    6564  283.48  6739.9  288.22  6970.3  293.12  7179.6  295.12
#Mann= 20 ,-1 , 0
  -354.1     .16       0  -117.1     .16       0   332.3     .05       0
    1645     .07       0  2050.7     .05       0  2271.2     .07       0
  2379.2     .05       0  2499.3     .07       0  2700.8     .12       0
  3798.4     .12       0  4335.4     .07       0  4605.7     .12       0
  4738.1     .07       0  4993.8     .07       0  4999.8     .07       0
  5105.7     .07       0  5314.1     .12       0    6564     .16       0
  6739.9     .16       0  6970.3     .16       0
#XS Ineff= 1 ,-1
 4297.48 4376.07  251.62
Permanent Ineff=
       F
Bank Sta=4916.7,5036.9
XS Rating Curve= 0 ,0
Exp/Cntr=0.3,0.1

Type RM Length L Ch R = 1 ,59720   ,1447,1447,1447
BEGIN DESCRIPTION:
TEHUACANA CREEK 23.0
END DESCRIPTION:
XS GIS Cut Line= 3
      3613749.62     10687710.16      3616949.61     10680510.19
      3616749.61     10678910.19
#Sta/Elev= 30
 -2917.1  310.64 -1969.9  306.11 -1350.2  280.74  -953.7  273.85    -630  269.61
    -446  256.41  -236.7  253.53  1724.1  249.24    1984  248.65    2432  249.26
  2975.6   249.5    3178  249.67    3306  249.99  3499.5  250.46  3732.7  250.74
    3972  250.82  4586.2  250.28  4940.1   250.8  4979.1   237.7  4981.9   237.2
  4985.1   237.7  4991.6  237.74  5032.5  251.18  5289.5  248.86  5418.8  248.95
  5786.8  257.09  5972.3  261.81  6214.1  287.36  6558.7  298.27  6574.4  298.79
#Mann= 20 ,-1 , 0
 -2917.1     .05       0  -953.7     .05       0  -236.7     .05       0
  1724.1     .07       0    1984     .05       0    2432     .05       0
  2975.6     .07       0    3178     .07       0    3306     .12       0
  3499.5     .12       0  3732.7     .07       0    3972     .12       0
  4586.2     .12       0  4979.1     .07       0  4985.1     .12       0
  4991.6     .07       0  5289.5     .07       0  5418.8     .12       0
  5786.8     .12       0  6558.7     .16       0
Bank Sta=4940.1,5032.5
XS Rating Curve= 0 ,0
Exp/Cntr=0.3,0.1

Type RM Length L Ch R = 1 ,58273   ,915,915,915
BEGIN DESCRIPTION:
TEHUACANA CREEK 22.0
END DESCRIPTION:
XS GIS Cut Line= 3
      3615049.63     10688110.15      3618249.61     10680110.19
      3616849.63     10678910.21
#Sta/Elev= 30
 -3630.7  302.39 -3124.5  277.43 -2699.7   270.8 -2688.6  270.71 -2291.9  268.22
 -2163.8  267.39  -791.4  259.96   237.2  264.65  1108.2  247.22  2043.1  248.58
  2209.8  249.32  2389.9  249.39  2770.9  249.46    3285  249.49  3289.9  249.43
  4606.3  249.82  4816.9  250.17 4918.18  251.43  5018.2  237.17  5020.9  236.67
  5024.2  237.17  5049.7  248.85  5070.6  243.21  5205.6  249.95    5909  251.25
  5982.6  253.54  6107.2  260.17  6220.3  267.04  6792.1  296.14  6829.4  298.27
#Mann= 20 ,-1 , 0
 -3630.7     .05       0 -2699.7     .08       0 -2688.6     .05       0
 -2291.9     .15       0 -2163.8     .05       0  2043.1     .07       0
  2209.8     .05       0  2389.9     .07       0  2770.9     .12       0
    3285     .07       0  3289.9     .12       0  4606.3     .07       0
  4816.9     .12       0  5018.2     .07       0  5024.2     .12       0
    5909     .16       0  5982.6     .12       0  6107.2     .16       0
  6220.3     .12       0  6792.1     .16       0
Bank Sta=4918.18,5205.6
XS Rating Curve= 0 ,0
Exp/Cntr=0.3,0.1

Type RM Length L Ch R = 1 ,57358   ,945,945,945
BEGIN DESCRIPTION:
TEHUACANA CREEK 21.0
END DESCRIPTION:
XS GIS Cut Line= 3
      3616095.88     10688825.53      3619038.62      10686195.3
      3618960.49     10678200.55
#Sta/Elev= 30
   -5463  301.51 -5272.2  298.49 -5095.8  284.35 -4853.6  272.57   -4445  257.19
 -3912.9  250.56 -3827.6  255.49 -3792.5  250.18    -131  248.82    62.1  257.01
   179.1  261.79   793.8  252.46  2089.2  247.24  2109.2  243.43  2129.2  247.33
  4138.6  249.07    4425  249.18  4959.3  250.58  4979.3  248.15  4989.3  241.01
  5006.3  237.26    5009  236.76  5012.3  237.26  5039.3  237.71  5049.3  247.88
  5139.3  249.07  5217.6  256.15  5409.3  270.95  5759.3  269.63    6479  294.17
#Mann= 10 ,-1 , 0
   -5463     .05       0 -4853.6     .16       0   -4445     .12       0
    62.1     .05       0   793.8     .12       0  4138.6     .07       0
    4425     .12       0  5006.3     .07       0  5012.3     .12       0
  5217.6     .05       0
#XS Ineff= 2 , 0
          172.73  261.84
Permanent Ineff=
       F       F
Bank Sta=4959.3,5217.6
XS Rating Curve= 0 ,0
Exp/Cntr=0.3,0.1

Type RM Length L Ch R = 1 ,56413   ,1411,1411,1411
BEGIN DESCRIPTION:
TEHUACANA CREEK 20.0
END DESCRIPTION:
XS GIS Cut Line= 3
      3616425.73     10689103.31      3621764.31     10685848.08
      3619429.24     10678070.29
#Sta/Elev= 30
 -7878.3  290.34 -7779.3  288.28 -7551.6  269.77   -7312  255.51 -6694.8     251
 -6436.4  250.43 -6401.7  250.42 -6137.5  250.33 -6033.5  256.24 -5959.9  248.26
   -5654  247.66   648.1  246.79   786.4  246.86  3660.1  243.56  3731.4  249.25
  4313.1  243.77  4720.3  249.57  4742.1  241.16  4835.2  240.34  4866.5  240.56
  4874.3  249.74  4960.5  249.58  5013.9  237.12  5016.6  236.62  5019.9  237.12
  5075.3  250.41  5368.3  249.98  5452.2  258.73  5714.4  279.92  6495.2   286.2
#Mann= 13 ,-1 , 0
 -7878.3     .16       0 -7779.3     .12       0 -7551.6     .16       0
   -7312     .12       0 -6694.8     .07       0 -6436.4     .12       0
 -6401.7     .07       0 -6137.5     .12       0   648.1     .07       0
   786.4     .12       0  5013.9     .07       0  5019.9     .12       0
  5452.2     .05       0
Bank Sta=4960.5,5075.3
XS Rating Curve= 0 ,0
Exp/Cntr=0.3,0.1

Type RM Length L Ch R = 1 ,55002   ,3244,3244,3244
BEGIN DESCRIPTION:
TEHUACANA CREEK 19.0
END DESCRIPTION:
XS GIS Cut Line= 3
      3652833.06     10683175.37      3625668.09     10681783.01
      3618251.42       10676783.
#Sta/Elev= 30
  -28120  307.27-25132.6  244.31-24712.1   263.1-24321.6  233.16-18012.1  242.46
-16363.7  244.46  -15876  247.01-15225.3   247.2-13614.3  247.88  -11897  243.16
  -11426  244.11-11384.6  225.08-11229.7  227.88-11194.4  247.75-10276.9  235.97
  -968.6  248.01  1293.6  248.65  1696.1   248.8    2753   247.9  3365.8  245.88
  4154.7  247.11  4945.3  250.35    4997  225.08  4999.8  224.58    5003  225.08
  5053.2  249.56  5352.8   256.1  5967.7  288.78  7748.1  295.56  8025.3  297.21
#Mann= 20 ,-1 , 0
  -28120     .07       0-18012.1     .07       0-16363.7     .12       0
  -15876     .05       0-15225.3     .07       0-13614.3     .07       0
  -11897     .12       0  -11426     .05       0-11229.7     .12       0
-10276.9     .12       0  -968.6     .07       0  1293.6     .12       0
  1696.1     .07       0    2753     .07       0  3365.8     .07       0
  4154.7     .12       0    4997     .07       0    5003     .12       0
  5352.8     .05       0  7748.1     .16       0
Bank Sta=4945.3,5053.2
XS Rating Curve= 0 ,0
Exp/Cntr=0.3,0.1

Type RM Length L Ch R = 1 ,51758   ,2242,2242,2242
BEGIN DESCRIPTION:
TEHUACANA CREEK 18.0
END DESCRIPTION:
XS GIS Cut Line= 3
      3653536.17     10682836.83      3628711.93     10679562.09
      3617774.52     10673468.39
#Sta/Elev= 30
-27253.8  301.66-24949.9  282.13-24100.1  241.64  -23188  266.34-22355.2  232.93
-16550.2  242.87-10331.1  243.62 -9968.1  244.19 -8426.1  244.37 -8208.7  232.53
   -8012  216.25 -7944.7  245.45   453.1  245.49   841.8  245.51  2800.3  245.59
  4074.4  247.04  4663.1  247.53  4970.9  247.06    4997  216.25  4999.8  215.75
    5003  216.25  5057.8  248.07  5062.2  248.04    5413  246.44  6151.9  249.63
  6438.6  252.59  6725.2  254.38  7612.1  265.44  8999.2  267.51 10305.9  306.74
#Mann= 20 ,-1 , 0
-27253.8     .07       0-16550.2     .07       0-10331.1     .12       0
 -9968.1     .07       0 -8426.1     .12       0 -8208.7     .05       0
 -7944.7     .12       0   453.1     .07       0   841.8     .12       0
  2800.3     .07       0  4074.4     .12       0  4663.1     .05       0
    4997     .03       0    5003     .05       0  5062.2     .12       0
    5413     .12       0  6151.9     .12       0  6438.6     .12       0
  6725.2     .05       0  7612.1     .05       0
Bank Sta=4970.9,5057.8
XS Rating Curve= 0 ,0
Exp/Cntr=0.3,0.1

Type RM Length L Ch R = 1 ,49516   ,2263,2263,2263
BEGIN DESCRIPTION:
TEHUACANA CREEK 17.0
END DESCRIPTION:
XS GIS Cut Line= 4
      3654389.29      10681105.2      3640390.17      10678578.3
      3629801.34     10677595.95      3617778.73     10672040.37
#Sta/Elev= 30
-26600.5  300.76-25647.1  275.63-23334.6  266.85-22983.3  238.16-14845.1  241.58
 -6639.8  244.65 -6532.5  244.77 -5655.9  245.75 -5516.6  216.39 -5390.3  231.48
    -411  244.91  4122.4  245.09  4962.1  246.54    4997  216.21  4999.8  215.71
    5003  216.21  5030.9  245.29  5234.2  247.01  5954.7  246.77  6061.7  247.99
  6281.3   245.5    7828  249.76  8263.6  253.02  8845.6  293.05  8952.7  294.64
  9670.2  273.54 10300.6  276.87 10665.9  282.28   10880  286.22 11503.3  311.89
#Mann= 20 ,-1 , 0
-26600.5     .07       0-14845.1     .07       0 -6639.8     .12       0
 -6532.5     .07       0 -5516.6     .05       0 -5390.3     .12       0
    -411     .12       0  4122.4     .12       0    4997     .07       0
    5003     .12       0  5954.7     .05       0  6061.7     .07       0
  6281.3     .05       0    7828     .05       0  8845.6     .08       0
  8952.7     .05       0  9670.2     .16       0 10300.6     .16       0
 10665.9     .16       0   10880     .05       0
Bank Sta=4962.1,5234.2
XS Rating Curve= 0 ,0
Exp/Cntr=0.3,0.1

Type RM Length L Ch R = 1 ,47253   ,6434,6434,6434
BEGIN DESCRIPTION:
Mapping XS 874d2eaf
END DESCRIPTION:
XS GIS Cut Line= 3
      3655262.18      10677207.9      3635576.73     10676502.34
      3617834.18     10670808.06
#Sta/Elev= 30
-26569.4  301.43-24945.8  297.72  -23655  246.96-22307.5  232.54-14207.9  237.87
-13812.4  238.13 -4628.7  244.17 -4112.2  215.05 -4070.9  244.61 -4017.7  244.73
 -1065.3  242.51    61.7  242.93   478.7  243.09  4951.4  244.16    4997  215.05
  4999.8  214.55    5003  215.05  5003.9  239.75  5035.7  243.73  5493.2  247.29
  7824.9  249.11  8054.3  255.89    8297  265.36  9325.3   310.4  9838.4     301
 10351.6   308.4 10703.1  313.47   11378  313.54 11705.3  316.41 11762.6  317.28
#Mann= 20 ,-1 , 0
-26569.4     .07       0-14207.9     .07       0-13812.4     .07       0
 -4628.7     .12       0 -4017.7     .12       0 -1065.3     .07       0
    61.7     .07       0   478.7     .12       0    4997     .07       0
    5003     .12       0  5493.2     .05       0  7824.9     .05       0
  8054.3     .16       0    8297     .05       0  9325.3     .05       0
  9838.4     .16       0 10351.6     .16       0 10703.1     .05       0
   11378     .12       0 11705.3     .16       0
Bank Sta=4951.4,5035.7
XS Rating Curve= 0 ,0
Exp/Cntr=0.3,0.1

Type RM Length L Ch R = 1 ,40819   ,4631,4631,4631
BEGIN DESCRIPTION:
TEHUACANA CREEK 15.0
END DESCRIPTION:
XS GIS Cut Line= 3
      3654240.08     10677032.96      3638232.98     10675175.14
      3616410.04     10662336.58
#Sta/Elev= 30
-24946.9  301.52-22108.2  261.63-21855.8  233.76-12985.2  238.83-12886.1  238.86
-12786.9  238.89   -3352  243.42 -3094.8  241.71 -2982.5  216.33 -2863.6  218.53
 -2830.1  244.38  4943.3   243.8    4997  214.85  4999.8  214.35    5003  214.85
  5024.6  243.32  5590.4   241.8  5771.2  249.58  5883.4   250.2  5926.3  250.14
    6188  249.75  6785.7  248.86  6893.4   248.7  7005.6  248.53  7140.3  248.33
  7187.6  248.26 11305.1  303.27 12168.2  346.59   15068  348.85   16487  399.49
#Mann= 20 ,-1 , 0
-24946.9     .07       0-12985.2     .05       0-12886.1     .08       0
-12786.9     .07       0   -3352     .12       0 -3094.8     .07       0
 -2982.5     .05       0 -2863.6     .12       0    4997     .07       0
    5003     .12       0  5590.4     .07       0  5771.2     .12       0
  5883.4     .05       0  5926.3     .07       0    6188     .05       0
  6785.7     .05       0  6893.4     .07       0  7005.6     .05       0
  7140.3     .07       0  7187.6     .05       0
Bank Sta=4943.3,5024.6
XS Rating Curve= 0 ,0
Exp/Cntr=0.3,0.1

Type RM Length L Ch R = 1 ,36188   ,959,959,959
BEGIN DESCRIPTION:
TEHUACANA CREEK 14.0
END DESCRIPTION:
XS GIS Cut Line= 3
      3654254.39     10676967.53      3644974.86     10675031.76
      3620028.79     10661762.48
#Sta/Elev= 30
-23001.1   301.3-20545.4  245.23-19972.5   251.4-19921.4  235.36-11433.5  240.23
-11303.9  240.21-11168.7  240.19-11060.4  240.17 -8478.3   239.7 -8339.2  241.97
 -8206.5  217.02 -8009.8  215.17   -7900  241.27 -7790.2  243.92 -7570.6  235.24
 -7455.4  249.15 -7198.1  237.07  -251.5   239.1  4892.9  244.53    4997  215.08
  4999.8  214.58    5003  215.08  5003.3  232.88  5019.1  239.82  6780.4  245.38
  6922.9  245.69  7032.7  249.82  7142.4  253.71  8377.7  279.47 14733.8  332.45
#Mann= 20 ,-1 , 0
-23001.1     .07       0-11433.5     .05       0-11303.9     .07       0
-11168.7     .05       0-11060.4     .07       0 -8478.3     .05       0
 -8339.2     .07       0 -8206.5     .05       0 -8009.8     .07       0
   -7900     .12       0 -7790.2     .12       0 -7570.6     .05       0
 -7198.1     .07       0  -251.5     .12       0    4997     .07       0
    5003     .12       0  6780.4     .07       0  6922.9     .05       0
  7032.7     .07       0  7142.4     .05       0
Bank Sta=4892.9,5019.1
XS Rating Curve= 0 ,0
Exp/Cntr=0.3,0.1

Type RM Length L Ch R = 1 ,35229   ,3983,3983,3983
BEGIN DESCRIPTION:
TEHUACANA CREEK 13.0
END DESCRIPTION:
XS GIS Cut Line= 4
      3652113.21     10675919.26      3629257.66      10666058.4
      3628762.87     10665146.94       3628788.9     10662543.99
#Sta/Elev= 30
-20521.4  286.88  -19570  233.03  -17163  236.93-16136.6  234.77-14619.2  235.79
-13846.6  237.86-12233.1  241.85-12151.7  212.27-11863.6  213.27-11782.9  241.75
 -8626.8   241.3 -7829.6  241.55 -7404.6  221.61 -7306.2  243.76 -4405.2  242.37
 -3708.5  234.82  -735.2   236.4    99.7     240     677  241.33  2959.9  244.34
  4981.1  239.54  4994.4  236.92    4997  212.27  4999.8  211.77    5003  212.27
  5090.4  242.53  5425.8  242.27  6113.6  253.53  7405.5  287.11  8010.8   294.7
#Mann= 20 ,-1 , 0
-20521.4     .07       0  -17163     .05       0-16136.6     .07       0
-14619.2     .05       0-13846.6     .07       0-11863.6     .07       0
 -8626.8     .12       0 -7829.6     .05       0 -7306.2     .07       0
 -4405.2     .07       0 -3708.5     .07       0  -735.2     .07       0
    99.7     .12       0     677     .07       0  2959.9     .12       0
    4997     .07       0    5003     .12       0  5425.8     .05       0
  6113.6     .12       0  7405.5     .12       0
Bank Sta=4981.1,5090.4
XS Rating Curve= 0 ,0
Exp/Cntr=0.3,0.1

Type RM Length L Ch R = 1 ,31246   ,5572,5572,5572
BEGIN DESCRIPTION:
TEHUACANA CREEK 12.0
END DESCRIPTION:
XS GIS Cut Line= 3
      3653068.13     10675789.08      3631757.34     10665792.54
      3632590.68     10662646.66
#Sta/Elev= 30
-18990.2  273.39-16948.4  232.95-10534.7  241.48-10224.4  242.65-10201.5  212.27
-10157.9  212.27 -9812.2  240.96 -9512.7  241.55 -9299.2  242.87 -9172.4  212.27
 -9021.1  227.87 -6957.4  241.69 -6574.9  241.92   -6036  243.82 -5978.9   243.4
 -5961.6  221.24 -5757.1  222.51 -5493.9  241.13 -4898.5  238.03  -807.9  242.08
  -657.1  242.23  4591.3  238.28  4968.9  238.95    4997  212.27  4999.8  211.77
    5003  212.27  5045.6  231.19  5084.4  239.67  5380.5  245.21  7803.1  306.08
#Mann= 20 ,-1 , 0
-18990.2     .07       0-10534.7     .12       0-10157.9     .05       0
 -9812.2     .12       0 -9512.7     .12       0 -9299.2     .05       0
 -9021.1     .07       0 -6957.4     .07       0 -6574.9     .12       0
   -6036     .05       0 -5757.1     .07       0 -5493.9     .07       0
 -4898.5     .07       0  -807.9     .08       0  -657.1     .07       0
  4591.3     .12       0    4997     .07       0    5003     .12       0
  5045.6     .07       0  5380.5     .05       0
Bank Sta=4968.9,5084.4
XS Rating Curve= 0 ,0
Exp/Cntr=0.3,0.1

Type RM Length L Ch R = 1 ,25674   ,2760,2760,2760
BEGIN DESCRIPTION:
Mapping XS 74c18680
END DESCRIPTION:
XS GIS Cut Line= 3
      3654072.49      10675631.1      3635582.86      10667141.5
      3633104.02     10664009.07
#Sta/Elev= 30
-15859.7  299.53-14649.4  292.08-13037.8  234.81-11845.9  236.95-10115.8  236.53
-10089.5  212.27 -8973.5  212.27 -8429.4  234.33 -7689.9  240.84 -7024.5  240.06
 -6114.2  241.96 -6096.7  212.27 -5713.4  239.14 -5305.1  212.27 -5090.8  239.67
 -2613.4  239.97 -1634.6  221.17 -1082.5   243.4  3862.7  238.52  4487.2  235.07
  4945.3  238.88    4997  212.27  4999.8  211.77    5003  212.27  5052.2  232.67
  5065.4  235.14  5848.9  245.78  7855.5  276.84  8463.4  291.78  8480.4  292.01
#Mann= 20 ,-1 , 0
-15859.7     .12       0-11845.9     .07       0-10115.8     .05       0
 -8973.5     .05       0 -8429.4     .07       0 -7689.9     .07       0
 -7024.5     .12       0 -5713.4     .07       0 -5090.8     .07       0
 -2613.4     .12       0 -1634.6     .07       0 -1082.5     .07       0
  3862.7     .07       0  4487.2     .12       0    4997     .07       0
    5003     .12       0  5052.2     .07       0  5848.9     .05       0
  7855.5     .05       0  8463.4     .08       0
Bank Sta=4945.3,5065.4
XS Rating Curve= 0 ,0
Exp/Cntr=0.3,0.1

Type RM Length L Ch R = 1 ,22914   ,825,825,825
BEGIN DESCRIPTION:
TEHUACANA CREEK 11.0
END DESCRIPTION:
XS GIS Cut Line= 3
      3655140.16     10674745.67      3639332.86     10667063.37
      3633890.12     10662297.72
#Sta/Elev= 30
-16572.8  301.56-14950.9  301.36-12887.4  239.94-11900.8  238.11-11891.3  212.27
-11625.8  236.92-11329.7  237.04 -6615.7  241.05 -6282.7  241.53 -5777.7  242.26
 -5433.7  242.75 -5411.2  212.27   -5035  237.85 -4700.8  212.92   -4576  241.79
 -3939.2  224.73   -2772   241.9  1641.2  241.83  2381.4  241.39  2710.3   241.2
  4443.4  240.17  4918.6  239.89    4997  212.27  4999.8  211.77    5003  212.27
  5159.7  239.34  5473.2  239.15  5883.6  243.37  6551.3  256.88  8236.7  302.71
#Mann= 20 ,-1 , 0
-16572.8     .12       0-11900.8     .05       0-11625.8     .12       0
-11329.7     .07       0 -6615.7     .12       0 -6282.7     .07       0
 -5777.7     .07       0   -5035     .05       0   -4576     .12       0
 -3939.2     .12       0   -2772     .07       0  1641.2     .12       0
  2381.4     .12       0  2710.3     .07       0  4443.4     .07       0
    4997     .07       0    5003     .07       0  5473.2     .05       0
  5883.6     .12       0  6551.3     .05       0
Bank Sta=4918.6,5159.7
XS Rating Curve= 0 ,0
Exp/Cntr=0.3,0.1

Type RM Length L Ch R = 1 ,22089   ,1516,1516,1516
BEGIN DESCRIPTION:
TEHUACANA CREEK 10.0
END DESCRIPTION:
XS GIS Cut Line= 3
      3649498.12     10667290.51       3636946.7     10664288.13
      3635149.62      10661810.2
#Sta/Elev= 30
 -8669.2  280.79 -8046.6  252.07   -7951  267.74 -7395.2  272.28   -6670  239.43
 -4938.3   241.4 -4904.5   239.1 -4886.9  212.27 -4263.4  238.52 -1856.3   242.3
 -1756.6   242.2 -1587.3  242.41  1311.8  241.81    1813  241.24  1927.9  240.92
  2008.7   240.7  2033.1  240.63  2077.6  240.29  4793.8  238.47  4949.7  238.51
    4997  212.27  4999.8  211.77    5003  212.27  5062.5  234.11  5183.8     237
  5219.6  240.74  5329.2   240.9  5967.9  247.52    5969  247.53  7297.3  275.83
#Mann= 18 ,-1 , 0
 -8669.2     .07       0 -1856.3     .05       0 -1756.6     .08       0
 -1587.3     .07       0  1311.8     .12       0    1813     .07       0
  1927.9     .12       0  2008.7     .07       0  2033.1     .12       0
  2077.6     .07       0  4793.8     .12       0    4997     .07       0
    5003     .12       0  5183.8     .07       0  5219.6     .05       0
  5329.2     .12       0  5967.9     .07       0    5969     .05       0
Bank Sta=4949.7,5062.5
XS Rating Curve= 0 ,0
Exp/Cntr=0.3,0.1

Type RM Length L Ch R = 1 ,20573   ,3618,3618,3618
BEGIN DESCRIPTION:
Mapping XS a715be54
END DESCRIPTION:
XS GIS Cut Line= 3
      3648695.22     10666661.18      3638722.94     10664139.65
      3634244.16     10658549.86
#Sta/Elev= 30
 -6845.3  277.91 -5591.4   238.7 -4741.5  238.76 -4248.5  238.34 -3652.3  240.74
 -3621.3  212.27 -3391.7  212.27 -3355.9  239.02 -2161.3   241.2 -1658.6  234.17
 -1370.1  239.97  -189.5   241.9   288.7  241.65  4951.6  233.15    4997  212.27
  4999.8  211.77    5003  212.27  5065.3  236.72  5275.6  238.48  6380.8   242.9
    6505  243.27  6769.9  244.07  6939.5  244.58    7975  252.44  8741.7  290.73
  9343.9  307.35  9842.1  309.35 10214.1  310.16 10553.7  310.89 10603.6  311.78
#Mann= 20 ,-1 , 0
 -6845.3     .07       0 -4741.5     .12       0 -4248.5     .07       0
 -2161.3     .12       0 -1658.6     .07       0 -1370.1     .07       0
  -189.5     .05       0   288.7     .07       0    4997     .07       0
    5003     .07       0  5275.6     .12       0  6380.8     .05       0
    6505     .07       0  6769.9     .12       0  6939.5     .05       0
  8741.7     .16       0  9343.9     .05       0  9842.1     .16       0
 10214.1     .05       0 10553.7     .08       0
Bank Sta=4951.6,5065.3
XS Rating Curve= 0 ,0
Exp/Cntr=0.3,0.1

Type RM Length L Ch R = 1 ,16955   ,2193,2193,2193
BEGIN DESCRIPTION:
TEHUACANA CREEK 9.0
END DESCRIPTION:
XS GIS Cut Line= 3
      3648722.97     10666466.05      3642125.72     10663271.59
      3634799.32     10657889.64
#Sta/Elev= 30
 -3721.9  281.22 -3214.1  274.69 -2273.7   238.1  -600.9  239.65  -115.1  241.71
   -92.5  237.98   -78.5  212.27   -75.7  211.77   -72.5  212.27   -69.9  226.47
   -62.8  212.27    93.7  212.27   124.8  230.97   466.4  235.48  2401.5  239.02
  3458.5  240.82  4771.6  242.29  4993.1  218.75  5187.5  240.21  6485.1  241.09
  6803.7  241.36  7109.9  241.01  7604.5  240.31  8236.3  239.89  8601.9  239.46
 10106.9  237.77 10685.2  243.19 10986.7   254.1 12434.3  310.06 12698.8  311.46
#Mann= 20 ,-1 , 0
 -3721.9     .05       0 -3214.1     .12       0 -2273.7     .07       0
  -600.9     .12       0   -78.5     .07       0   -72.5     .05       0
   124.8     .12       0   466.4     .07       0  2401.5     .12       0
  3458.5     .07       0  6485.1     .05       0  6803.7     .12       0
  7109.9     .07       0  7604.5     .07       0  8236.3     .07       0
  8601.9     .07       0 10106.9     .05       0 10685.2     .05       0
 10986.7     .16       0 12434.3     .05       0
#XS Ineff= 1 ,-1
 -144.32 1205.68  241.75
Permanent Ineff=
       F
Bank Sta=4771.6,5187.5
XS Rating Curve= 0 ,0
Exp/Cntr=0.3,0.1

Type RM Length L Ch R = 1 ,14762   ,1850,1850,1850
BEGIN DESCRIPTION:
TEHUACANA CREEK 8.0
END DESCRIPTION:
XS GIS Cut Line= 3
      3648584.09     10665979.96      3642299.33     10660910.48
       3634973.8     10657716.41
#Sta/Elev= 30
 -3777.1   274.8 -2446.8  240.39  -648.1  236.22   -75.5  237.68   341.2  239.12
   805.3  242.13   869.3  230.22   877.3  212.27  1200.6  209.65  1203.3  209.15
  1206.6  209.65  1232.3  209.65  1239.3   229.9  1261.1  236.56    1667  236.67
  3336.4  238.05  4813.2  238.16  5011.4  217.46  5448.1  239.02  5783.2  240.51
  6478.8  240.63  7024.1  240.26  7359.5   239.6    8288  237.78  9940.2  234.99
 10436.3  244.98 10639.6  248.37 11925.7  307.29 12285.2  309.84   12289  309.88
#Mann= 20 ,-1 , 0
 -3777.1     .05       0 -2446.8     .07       0  -648.1     .12       0
   -75.5     .07       0   341.2     .12       0  1200.6     .07       0
  1206.6     .12       0    1667     .07       0  3336.4     .07       0
  5448.1     .05       0  5783.2     .05       0  6478.8     .05       0
  7024.1     .05       0  7359.5     .07       0    8288     .07       0
  9940.2     .05       0 10436.3     .12       0 10639.6     .16       0
 11925.7     .05       0 12285.2     .05       0
#XS Ineff= 1 ,-1
  755.68  1287.5  241.45
Permanent Ineff=
       F
Bank Sta=4813.2,5448.1
XS Rating Curve= 0 ,0
Exp/Cntr=0.3,0.1

Type RM Length L Ch R = 1 ,12912   ,2917,2917,2917
BEGIN DESCRIPTION:
TEHUACANA CREEK 7.0
END DESCRIPTION:
XS GIS Cut Line= 3
      3648549.32     10665146.59      3642438.22     10659035.48
      3635146.56     10657125.76
#Sta/Elev= 30
 -4208.1  263.23 -3440.1     264 -2645.1   235.1   -1184   235.5  1302.2  237.79
  2108.7  240.24  2536.1  238.22  2619.8   216.2  2765.3  216.19    2768  215.69
  2771.3  216.19  2817.8  239.27  4552.8  241.04  4906.2  232.77  4992.1  216.73
  5053.1  232.06  5357.3  238.24  5380.1  238.86  5426.3  239.59  7454.1  240.54
  7699.7   239.4  7802.2  238.85  7971.7  237.94  9926.3  239.68 10434.6  248.51
 10535.9  257.07 10659.5  255.48   11019  275.11 11509.8  306.05 11971.9   311.2
#Mann= 20 ,-1 , 0
 -4208.1     .05       0 -2645.1     .07       0   -1184     .12       0
  1302.2     .07       0  2108.7     .12       0  2536.1     .05       0
  2765.3     .07       0  2771.3     .05       0  5357.3     .05       0
  5380.1     .05       0  7454.1     .07       0  7699.7     .07       0
  7802.2     .05       0  7971.7     .07       0  9926.3     .05       0
 10434.6     .08       0 10535.9      .1       0 10659.5     .05       0
   11019     .12       0 11509.8     .05       0
#XS Ineff= 1 ,-1
 2464.23 2842.36  238.71
Permanent Ineff=
       F
Bank Sta=4552.8,5426.3
XS Rating Curve= 0 ,0
Exp/Cntr=0.3,0.1

Type RM Length L Ch R = 1 ,9995    ,3556,3556,3556
BEGIN DESCRIPTION:
TEHUACANA CREEK 6.0
END DESCRIPTION:
XS GIS Cut Line= 4
      3648089.27      10664480.9       3642338.4     10657080.73
      3642077.99     10656190.98      3643705.08     10652177.46
#Sta/Elev= 30
   -4882  266.53 -3761.9   239.2 -2436.2  238.82  -647.4   238.3   372.8     238
  1347.3  238.93  1447.4  222.92  1493.6  224.13  1536.9  207.68  1539.6  207.18
  1542.9  207.68  1641.2  214.94  1681.2  239.86  3758.4   239.1 4463.64   239.2
  4611.8  237.72    4764  236.33  4932.1   234.8  4986.3  217.16    5071  236.67
  7096.5  231.59  8007.7  259.68    8181  247.07  8872.3  308.92  9027.7  298.66
  9194.6  333.02  9377.7  349.54  9403.4  351.63  9551.8     365  9747.9  362.25
#Mann= 18 ,-1 , 0
   -4882     .05       0 -3761.9     .07       0 -2436.2     .12       0
  -647.4     .07       0   372.8     .12       0  1447.4     .08       0
  1493.6     .05       0  1536.9     .07       0  1542.9     .05       0
  1641.2     .07       0  3758.4     .12       0  4611.8     .07       0
    4764     .12       0  4986.3     .07       0  7096.5     .12       0
  9377.7     .16       0  9403.4     .12       0  9551.8     .16       0
#XS Ineff= 1 ,-1
 1341.98 1712.89  239.48
Permanent Ineff=
       F
Bank Sta=4463.64,5071
XS Rating Curve= 0 ,0
Exp/Cntr=0.3,0.1

Type RM Length L Ch R = 1 ,6439    ,1888,1888,1888
BEGIN DESCRIPTION:
TEHUACANA CREEK 4.0
END DESCRIPTION:
XS GIS Cut Line= 3
      3647915.67     10663482.66      3644768.96     10657861.98
       3644031.1     10654606.73
#Sta/Elev= 30
 -2143.5  264.69 -1014.2  236.27   877.9  234.83  2372.9  233.66  2387.3  227.88
  2397.6  208.25  2403.3  221.48  2406.1  207.68  2408.9  207.18  2412.1  207.68
  2472.1  207.68  2488.3  207.68  2638.4  207.68  2646.5   224.3  2661.3   234.8
  2681.8  235.58  3838.3  238.41  4658.8  236.23  4875.5  227.77  4884.6   228.3
  4966.4  228.34  4994.2  212.74  5042.4  212.28  5099.7  234.06  6397.7  229.62
  6655.7  240.06  6873.6  258.23  7440.9  336.71    7484  350.65  7635.9  353.42
#Mann= 13 ,-1 , 0
 -2143.5     .05       0 -1014.2     .07       0   877.9     .12       0
  2372.9     .07       0  2406.1     .07       0  2412.1     .07       0
  2472.1     .12       0  2488.3     .05       0  2681.8     .12       0
  3838.3     .07       0  4875.5     .05       0  4884.6     .07       0
  6655.7     .12       0
#XS Ineff= 1 ,-1
 2346.78 2718.33  237.33
Permanent Ineff=
       F
Bank Sta=4658.8,5099.7
XS Rating Curve= 0 ,0
Exp/Cntr=0.3,0.1

Type RM Length L Ch R = 1 ,4551    ,1548,1548,1548
BEGIN DESCRIPTION:
TEHUACANA CREEK 3.0
END DESCRIPTION:
XS GIS Cut Line= 3
      3647849.61     10663160.19      3646249.61     10656760.19
      3644649.62     10654760.21
#Sta/Elev= 30
 -1563.7  260.33  -715.9  249.23  -491.7  255.55    47.6  236.63  2524.9  232.84
  3023.3  238.92  3072.2  230.51  3082.1  207.68  3084.9  207.18  3088.1  207.68
  3136.6  207.68  3229.1  207.68  3358.9  207.68    3384  207.68  3402.1  229.67
  3484.5  240.05  3924.9   238.2  4672.5  237.72  4762.7  228.05  4884.1  229.15
  4971.2  228.66  5879.3  228.22  6100.2  235.07  6798.7  238.09  6901.9   245.3
  7075.1  257.54  7246.4  280.35    7360  302.32  7430.4  330.66  7594.5  353.56
#Mann= 13 ,-1 , 0
 -1563.7     .05       0    47.6     .07       0  2524.9     .12       0
  3082.1     .07       0  3088.1     .12       0  3136.6     .07       0
  3229.1     .05       0  3358.9     .12       0  3924.9     .07       0
  4884.1     .05       0  4971.2     .07       0  6798.7     .05       0
  6901.9     .12       0
#XS Ineff= 1 ,-1
 2988.64 3539.77  239.25
Permanent Ineff=
       F
Bank Sta=4672.5,6100.2
XS Rating Curve= 0 ,0
Exp/Cntr=0.3,0.1

Type RM Length L Ch R = 1 ,3003    ,791,791,791
BEGIN DESCRIPTION:
TEHUACANA CREEK 2.0
END DESCRIPTION:
XS GIS Cut Line= 3
      3648199.61     10663260.19      3647416.53     10655605.04
      3645599.61     10654060.19
#Sta/Elev= 30
 -2221.9  265.45   -1659  261.58    -451  239.18    1206  235.72  2452.4  237.29
  2673.5  232.26  3065.6  236.95  3075.6  235.36  3085.7  225.73  3092.7  207.68
  3095.5  207.18  3098.7  207.68  3113.6  207.68  3306.8  207.68  3316.9  232.58
  3329.1  236.37    3347  240.55  3649.8  238.67  4513.7  237.37  4889.3  229.61
  4898.3  229.85  5005.7  229.16  5176.5  237.96    6879  229.04  7171.7  237.26
    7326  251.75  7418.3  267.63  7510.5  305.49  7567.6  320.61  7858.1  339.59
#Mann= 11 ,-1 , 0
 -2221.9     .05       0    -451     .07       0    1206     .12       0
  3092.7     .07       0  3098.7     .12       0  3113.6     .05       0
  3329.1     .12       0  3649.8     .07       0  4889.3     .05       0
  4898.3     .07       0  7171.7     .12       0
#XS Ineff= 1 ,-1
    3050 3459.09  237.15
Permanent Ineff=
       F
Bank Sta=4513.7,5176.5
XS Rating Curve= 0 ,0
Exp/Cntr=0.3,0.1

Type RM Length L Ch R = 1 ,2212    ,0,0,0
BEGIN DESCRIPTION:
TEHUACANA CREEK 1.0
END DESCRIPTION:
XS GIS Cut Line= 3
      3649391.62     10663634.79      3647959.33     10655249.37
      3645278.18     10652333.95
#Sta/Elev= 30
 -3027.7  262.89 -2555.9  261.73 -2198.4  258.26 -2043.9  254.39 -1836.2  250.17
  -947.8  238.77  1238.8  237.52  2787.6  235.31  3063.9  229.21  3067.5  207.68
  3070.2  207.18  3073.5  207.68  3250.9  207.68  3256.6  233.27  3266.8  240.19
  3309.1  239.92  3642.5  237.43  4438.3  238.42  4922.1  222.44  5034.5  215.99
  5111.7  228.38  5209.9  236.82  5865.6  235.85  6266.8  235.51  7593.7  233.89
  8323.4  253.82  8924.7  306.64  9065.3  326.43  9255.3  332.29    9440  339.53
#Mann= 20 ,-1 , 0
 -3027.7     .05       0 -2555.9     .16       0 -2198.4     .05       0
 -2043.9     .16       0 -1836.2     .05       0  -947.8     .12       0
  1238.8     .07       0  2787.6     .12       0  3067.5    .033       0
  3073.5     .05       0  3309.1     .12       0  3642.5     .07       0
  4922.1     .05       0  5111.7     .07       0  5865.6     .12       0
  6266.8     .07       0  7593.7     .12       0  8924.7     .12       0
  9065.3     .05       0  9255.3     .16       0
#XS Ineff= 1 ,-1
 2753.41 3294.32  236.45
Permanent Ineff=
       F
Bank Sta=4438.3,5209.9
XS Rating Curve= 0 ,0
Exp/Cntr=0.3,0.1

Chan Stop Cuts=-1
Use User Specified Reach Order=0
Composite Channel Slope=5
