--- UNT166 IN CCTC.prj (project) ---

Proj Title=UNT166 IN CCTC Base Level Engineering
Current Plan=p01
Default Exp/Contr=0.3,0.1
English Units
Geom File=g01
Flow File=f01
Plan File=p01
Y Axis Title=Elevation
X Axis Title(PF)=Main Channel Distance
X Axis Title(XS)=Station
BEGIN DESCRIPTION:
UNT166 IN CCTC
END DESCRIPTION:
DSS Export Rating Curves= 0
DSS Export Rating Curve Sorted= 0
DSS Export Volume Flow Curves= 0
DXF OffsetX= 0
DXF OffsetY= 0
DXF ScaleX= 1
DXF ScaleY= 10

--- UNT166 IN CCTC.p01 (plan) ---

Plan Title=Multiple Run
Short Identifier=Multiple
Geom File=g01
Flow File=f01
Subcritical Flow
K Sum by GR= 0
Std Step Tol= 0.01
Critical Tol= 0.01
Num of Std Step Trials= 20
Max Error Tol= 0.3
Flow Tol Ratio= 0.001
Split Flow NTrial= 30
Split Flow Tol= 0.02
Split Flow Ratio= 0.02
Log Output Level= 0
Friction Slope Method= 1
Unsteady Friction Slope Method= 2
Unsteady Bridges Friction Slope Method= 1
Parabolic Critical Depth
Global Vel Dist=  1 , 1 , 1
Global Log Level= 0
CheckData=True
Encroach Param= -1, 0, 0, 0
BEGIN DESCRIPTION:
Multiple Run
END DESCRIPTION:

--- UNT166 IN CCTC.f01 (steady flow) ---

Flow Title=Multiple
Program Version=4.10
Number of Profiles= 7
Profile Names=10-year,25-year,50-year,1pct_min,100-year,1pct_plu,500-year
River Rch & RM=UNT166 IN CCTC,Reach-1         ,31718
    1935    2699    3337    3004    4063    5495    6011
River Rch & RM=UNT166 IN CCTC,Reach-1         ,24485
    2103    2937    3632    3269    4421    5979    6538
River Rch & RM=UNT166 IN CCTC,Reach-1         ,16667
    3329    4740    5942    5412    7319    9898   11086
River Rch & RM=UNT166 IN CCTC,Reach-1         ,11423
    3486    4971    6236    5685    7688   10397   11661
River Rch & RM=UNT166 IN CCTC,Reach-1         ,7432
    4178    5989    7539    6891    9319   12603   14213
River Rch & RM=UNT166 IN CCTC,Reach-1         ,6218
    4178    5989    7539    6891    9319   12603   14213
Boundary for River Rch & Prof#=UNT166 IN CCTC,Reach-1         , 1
Up Type= 0
Dn Type= 3
Dn Slope=0.005
Boundary for River Rch & Prof#=UNT166 IN CCTC,Reach-1         , 2
Up Type= 0
Dn Type= 3
Dn Slope=0.005
Boundary for River Rch & Prof#=UNT166 IN CCTC,Reach-1         , 3
Up Type= 0
Dn Type= 3
Dn Slope=0.005
Boundary for River Rch & Prof#=UNT166 IN CCTC,Reach-1         , 4
Up Type= 0
Dn Type= 3
Dn Slope=0.005
Boundary for River Rch & Prof#=UNT166 IN CCTC,Reach-1         , 5
Up Type= 0
Dn Type= 3
Dn Slope=0.005
Boundary for River Rch & Prof#=UNT166 IN CCTC,Reach-1         , 6
Up Type= 0
Dn Type= 3
Dn Slope=0.005
Boundary for River Rch & Prof#=UNT166 IN CCTC,Reach-1         , 7
Up Type= 0
Dn Type= 3
Dn Slope=0.005
DSS Import GetInterval= 0
DSS Import GetPeak= 0
DSS Import FillOption= 0

--- UNT166 IN CCTC.g01 (geometry) ---

Geom Title=Existing Conditions

River Reach=UNT166 IN CCTC,Reach-1
Reach XY= 30
      3552128.75     10676991.00      3552417.25     10676144.00
      3554123.75     10674681.00      3554451.25     10673909.00
      3555395.00     10673423.00      3555497.50     10671674.00
      3556734.75     10670842.00      3556756.75     10670325.00
      3557464.50     10670132.00      3557683.75     10669358.00
      3559162.25     10669364.00      3559979.25     10668841.00
      3560519.50     10668081.00      3561105.25     10668390.00
      3561353.25     10667988.00      3561809.50     10667910.00
      3562071.50     10668197.00      3562346.00     10668047.00
      3562524.25     10668408.00      3563061.25     10668045.00
      3563548.25     10667984.00      3563899.50     10668341.00
      3564585.00     10668044.00      3564859.75     10668361.00
      3565585.75     10668053.00      3565756.25     10667623.00
      3567360.00     10666269.00      3567886.75     10666627.00
      3568059.75     10667129.00      3568629.00     10666530.00

Type RM Length L Ch R = 1,31718,456,456,456
BEGIN DESCRIPTION:
UNT166 IN CCTC 53.0
END DESCRIPTION:
XS GIS Cut Line= 3
      3552399.60     10677610.14      3552249.61     10676860.19
      3551749.59     10676210.16
#Sta/Elev= 30
  4221.9  382.84  4242.2  381.26  4374.8  378.34  4466.6  374.84  4497.2  372.58
  4507.4  373.77  4568.6  371.35  4609.4  367.92  4619.6  366.02  4660.4  365.05
  4687.2  366.69  4721.6  368.73  4752.2  371.76  4803.1  372.37  4854.1  371.29
  4864.3  369.83  4894.9  369.40  4915.3  367.14  4976.5  365.41  4997.3  363.56
  5000.0  363.06  5003.3  363.56  5064.6  365.25  5207.8  365.61  5228.6  366.58
  5415.3  368.97  5515.0  373.14  5529.2  374.62  5685.3  383.14  5806.8  386.77
#Mann=4,-1,0
  4221.9    0.16       0  4687.2    0.05       0  4997.3    0.03       0
  5003.3    0.05       0
Bank Sta=4997.3,5003.3
Exp/Cntr=0.3,0.1

Type RM Length L Ch R = 1,31262,476,476,476
BEGIN DESCRIPTION:
UNT166 IN CCTC 52.0
END DESCRIPTION:
XS GIS Cut Line= 3
      3552749.57     10676710.17      3552249.61     10676460.19
      3551849.60     10676260.18
#Sta/Elev= 30
  4463.7  378.26  4522.4  376.02  4530.7  376.13  4553.1  374.75  4642.5  372.28
  4701.2  368.83  4732.0  368.10  4768.3  366.48  4829.8  364.60  4874.5  363.63
  4964.0  363.27  4983.3  362.72  4986.1  362.22  4989.3  362.72  5067.4  364.31
  5126.1  366.58  5134.5  366.26  5142.9  367.21  5193.2  369.05  5232.3  369.78
  5260.3  371.15  5277.0  371.39  5282.6  372.48  5299.4  372.80  5335.7  375.51
  5366.5  376.93  5380.4  378.02  5402.8  378.67  5416.8  379.94  5469.9  382.55
#Mann=3,-1,0
  4463.7    0.05       0  4983.3    0.03       0  4989.3    0.05       0
Bank Sta=4983.3,4989.3
Exp/Cntr=0.3,0.1

Type RM Length L Ch R = 1,30786,454,454,454
BEGIN DESCRIPTION:
UNT166 IN CCTC 51.0
END DESCRIPTION:
XS GIS Cut Line= 3
      3552799.62     10676510.20      3552449.61     10676110.19
      3552249.59     10675860.17
#Sta/Elev= 30
  4483.6  376.31  4497.4  375.29  4611.3  370.70  4625.5  369.21  4639.7  368.72
  4660.6  367.05  4696.2  365.84  4710.0  364.18  4746.0  362.38  4752.7  362.72
  4809.6  360.55  4844.8  360.55  4887.5  361.39  4962.3  360.26  4965.0  359.76
  4968.3  360.26  4993.8  361.04  5043.1  361.06  5100.8  363.78  5200.0  369.85
  5228.8  371.12  5243.2  373.58  5257.6  374.00  5264.0  374.94  5278.4  374.40
  5292.9  375.17  5299.3  376.12  5313.7  376.81  5328.1  379.46  5335.3  379.59
#Mann=3,-1,0
  4483.6    0.05       0  4962.3    0.03       0  4968.3    0.05       0
Bank Sta=4962.3,4968.3
Exp/Cntr=0.3,0.1

Type RM Length L Ch R = 1,30332,484,484,484
BEGIN DESCRIPTION:
UNT166 IN CCTC 50.0
END DESCRIPTION:
XS GIS Cut Line= 3
      3552849.61     10676460.19      3552799.61     10675810.19
      3552399.63     10675510.20
#Sta/Elev= 30
  4385.5  376.31  4395.5  375.40  4465.7  372.30  4525.9  370.75  4576.1  366.82
  4596.1  364.76  4616.2  363.68  4626.2  362.33  4646.3  361.56  4736.5  359.51
  4897.0  359.00  4954.2  357.52  4956.9  357.02  4960.2  357.52  4987.3  357.62
  4997.3  358.76  5040.5  358.78  5051.0  357.82  5059.3  357.80  5094.7  359.51
  5180.1  360.41  5209.3  361.53  5230.1  361.68  5259.3  363.71  5280.1  364.01
  5294.7  365.50  5365.5  368.58  5473.9  375.35  5487.4  376.71  5537.4  379.00
#Mann=3,-1,0
  4385.5    0.05       0  4954.2    0.03       0  4960.2    0.05       0
Bank Sta=4954.2,4960.2
Exp/Cntr=0.3,0.1

Type RM Length L Ch R = 1,29848,424,424,424
BEGIN DESCRIPTION:
UNT166 IN CCTC 49.0
END DESCRIPTION:
XS GIS Cut Line= 3
      3553499.59     10675910.17      3553149.61     10675510.19
      3552799.58     10675210.16
#Sta/Elev= 30
  4461.3  371.48  4539.6  370.25  4595.6  368.09  4638.3  364.94  4701.9  361.84
  4730.4  359.34  4744.6  357.41  4766.4  356.06  4808.2  355.37  4830.0  356.10
  4872.7  355.43  4928.7  356.97  5020.8  355.85  5049.3  356.15  5068.3  355.32
  5071.0  354.82  5074.3  355.32  5134.9  356.84  5155.8  356.40  5233.7  356.99
  5361.6  360.99  5375.3  362.46  5383.0  365.29  5397.2  367.87  5411.5  374.47
  5418.1  376.41  5425.8  376.52  5432.4  377.39  5446.6  372.97  5453.8  372.97
#Mann=3,-1,0
  4461.3    0.05       0  5068.3    0.03       0  5074.3    0.05       0
Bank Sta=5068.3,5074.3
Exp/Cntr=0.3,0.1

Type RM Length L Ch R = 1,29424,461,461,461
BEGIN DESCRIPTION:
UNT166 IN CCTC 48.0
END DESCRIPTION:
XS GIS Cut Line= 3
      3553749.63     10675560.22      3553449.61     10675210.19
      3553049.61     10674810.19
#Sta/Elev= 30
  4556.2  369.40  4570.0  368.21  4577.6  367.16  4584.2  365.57  4606.2  364.38
  4634.7  361.75  4662.2  360.08  4684.1  359.57  4690.7  358.61  4733.5  357.90
  4740.6  356.80  4882.8  354.45  4967.3  354.60  4995.8  354.05  5020.7  354.52
  5042.5  354.04  5045.2  353.54  5048.5  354.04  5102.1  354.28  5144.5  355.71
  5229.3  360.66  5243.5  361.97  5328.3  366.17  5342.5  367.26  5356.6  369.19
  5384.9  371.35  5469.8  377.11  5512.2  379.41  5526.3  380.93  5582.9  384.62
#Mann=3,-1,0
  4556.2    0.05       0  5042.5    0.03       0  5048.5    0.05       0
Bank Sta=5042.5,5048.5
Exp/Cntr=0.3,0.1

Type RM Length L Ch R = 1,28963,111,111,111
BEGIN DESCRIPTION:
UNT166 IN CCTC 47.0
END DESCRIPTION:
XS GIS Cut Line= 3
      3554149.59     10675110.18      3553799.61     10674910.19
      3553399.60     10674610.18
#Sta/Elev= 30
  4566.6  369.64  4641.2  365.04  4660.9  364.49  4676.7  362.37  4720.7  359.42
  4785.4  355.48  4838.0  354.01  5047.7  352.54  5061.8  352.92  5124.0  352.10
  5126.7  351.60  5130.0  352.10  5162.4  352.16  5169.7  354.61  5191.6  355.97
  5233.2  360.68  5306.1  364.35  5312.4  365.61  5333.2  366.78  5347.8  366.67
  5391.6  371.03  5406.1  371.61  5412.4  369.59  5422.2  372.06  5427.0  373.09
  5433.2  371.47  5441.6  372.86  5447.8  371.04  5462.4  371.13  5469.7  372.29
#Mann=8,-1,0
  4566.6    0.05       0  4641.2    0.08       0  4720.7    0.05       0
  5047.7    0.08       0  5061.8    0.05       0  5124.0    0.03       0
  5130.0    0.05       0  5422.2    0.08       0
Bank Sta=5124,5130
Exp/Cntr=0.3,0.1

Type RM Length L Ch R = 1,28852,793,793,793
BEGIN DESCRIPTION:
UNT166 IN CCTC 46.0
END DESCRIPTION:
XS GIS Cut Line= 3
      3554216.70     10675028.71      3553807.01     10674782.20
      3553435.47     10674528.72
#Sta/Elev= 30
  4559.8  370.53  4564.4  368.81  4570.3  370.05  4585.8  368.06  4604.4  368.54
  4673.1  364.73  4739.2  358.20  4788.6  356.64  4840.3  355.00  5014.3  353.80
  5030.6  355.16  5035.0  353.48  5051.7  353.42  5064.5  355.31  5072.6  353.55
  5102.5  353.74  5105.5  351.48  5108.3  350.98  5111.5  351.48  5131.6  351.52
  5138.4  353.31  5174.3  356.55  5180.3  355.89  5275.9  362.20  5282.0  364.40
  5347.7  368.08  5353.8  369.74  5383.6  369.85  5389.7  371.41  5487.7  375.87
#Mann=7,-1,0
  4559.8    0.05       0  4604.4    0.08       0  4788.6    0.05       0
  5014.3    0.08       0  5064.5    0.05       0  5105.5    0.04       0
  5111.5    0.05       0
Bank Sta=5105.5,5111.5
Exp/Cntr=0.3,0.1

Type RM Length L Ch R = 1,28059,420,420,420
BEGIN DESCRIPTION:
UNT166 IN CCTC 45.0
END DESCRIPTION:
XS GIS Cut Line= 3
      3554549.61     10674610.19      3554249.61     10674360.19
      3554049.59     10674060.17
#Sta/Elev= 30
  4623.0  369.27  4687.4  365.28  4701.1  363.80  4729.1  361.78  4772.1  360.07
  4786.4  358.34  4807.2  357.43  4821.5  356.11  4835.8  355.73  4850.2  354.53
  4949.1  349.76  4985.5  348.88  4996.9  347.71  4999.6  347.21  5002.9  347.71
  5006.4  348.96  5027.0  348.59  5042.1  349.70  5078.1  349.79  5093.1  348.98
  5121.7  348.83  5135.2  349.35  5186.3  349.70  5302.0  353.69  5324.5  356.74
  5330.5  358.83  5338.0  359.86  5345.5  363.09  5366.6  367.44  5374.1  367.00
#Mann=3,-1,0
  4623.0    0.05       0  4996.9   0.035       0  5002.9    0.05       0
Bank Sta=4996.9,5002.9
Exp/Cntr=0.3,0.1

Type RM Length L Ch R = 1,27639,428,428,428
BEGIN DESCRIPTION:
UNT166 IN CCTC 44.0
END DESCRIPTION:
XS GIS Cut Line= 3
      3554599.58     10674210.16      3554399.61     10674010.19
      3554099.65     10673960.20
#Sta/Elev= 30
  4723.3  361.34  4751.5  359.67  4836.4  353.23  4850.5  351.32  4878.8  349.17
  4893.0  348.74  4921.3  346.58  4935.4  347.34  4963.7  347.68  4999.6  345.13
  5002.3  344.63  5005.6  345.13  5026.4  345.71  5034.0  346.88  5077.1  348.44
  5107.5  349.33  5148.0  349.51  5168.3  350.60  5178.4  350.55  5208.9  351.64
  5216.5  351.97  5221.5  352.91  5249.4  353.97  5269.7  355.98  5277.3  358.82
  5282.4  359.29  5290.0  361.20  5300.1  365.14  5307.7  366.62  5310.2  366.62
#Mann=3,-1,0
  4723.3    0.05       0  4999.6   0.035       0  5005.6    0.05       0
Bank Sta=4999.6,5005.6
Exp/Cntr=0.3,0.1

Type RM Length L Ch R = 1,27211,417,417,417
BEGIN DESCRIPTION:
UNT166 IN CCTC 43.0
END DESCRIPTION:
XS GIS Cut Line= 3
      3554799.61     10674060.21      3554699.61     10673710.19
      3554449.63     10673410.22
#Sta/Elev= 30
  4663.1  360.26  4704.7  357.62  4735.9  354.01  4746.3  353.52  4758.0  351.73
  4777.5  350.34  4808.7  345.58  4819.1  346.02  4830.8  345.65  4839.9  346.42
  4859.4  346.71  4864.6  345.12  4871.1  345.82  4881.5  345.53  4898.4  346.53
  4903.6  345.65  4920.1  344.96  4922.9  344.46  4926.1  344.96  4932.2  346.05
  4964.7  346.36  5005.0  345.41  5176.2  348.05  5332.4  353.28  5375.3  356.71
  5396.2  363.19  5404.0  364.81  5410.5  368.23  5414.4  369.58  5417.6  369.58
#Mann=3,-1,0
  4663.1    0.05       0  4920.1   0.035       0  4926.1    0.05       0
Bank Sta=4920.1,4926.1
Exp/Cntr=0.3,0.1

Type RM Length L Ch R = 1,26794,555,555,555
BEGIN DESCRIPTION:
UNT166 IN CCTC 42.0
END DESCRIPTION:
XS GIS Cut Line= 2
      3555478.39     10674190.62      3554710.13     10673127.20
#Sta/Elev= 30
  4270.9  369.04  4363.3  367.06  4392.8  367.42  4478.6  364.99  4514.2  363.54
  4600.1  357.74  4706.8  351.97  4786.5  348.46  4973.0  343.99  4993.8  344.46
  5000.0  342.54  5008.5  342.39  5014.7  343.61  5023.3  342.92  5029.4  344.04
  5044.1  344.68  5079.7  344.95  5100.6  344.69  5133.2  342.22  5135.9  341.72
  5139.2  342.22  5165.6  343.35  5186.5  345.36  5209.0  349.55  5236.7  352.90
  5266.2  354.46  5307.9  358.60  5387.6  364.18  5480.4  365.98  5582.8  366.54
#Mann=3,-1,0
  4270.9    0.05       0  5133.2   0.035       0  5139.2    0.05       0
Bank Sta=5133.2,5139.2
Exp/Cntr=0.3,0.1

Type RM Length L Ch R = 1,26239,631,631,631
BEGIN DESCRIPTION:
UNT166 IN CCTC 41.0
END DESCRIPTION:
XS GIS Cut Line= 2
      3556181.55     10673609.02      3554802.93     10673023.76
#Sta/Elev= 30
  4161.2  370.70  4288.1  367.34  4358.9  364.98  4380.9  361.38  4399.1  360.97
  4404.5  358.85  4422.8  358.94  4428.2  363.04  4451.9  361.09  4489.2  363.04
  4587.0  360.69  4628.3  357.41  4681.1  355.95  4857.6  343.57  4939.4  341.63
  4969.7  336.93  4996.8  331.38  4999.6  330.88  5002.8  331.38  5010.4  335.54
  5015.8  333.65  5021.5  338.56  5075.9  342.17  5139.5  341.90  5268.7  346.80
  5390.9  354.18  5426.9  354.10  5467.0  358.88  5606.3  366.25  5658.9  368.70
#Mann=6,-1,0
  4161.2    0.05       0  4288.1    0.16       0  4969.7    0.05       0
  4996.8   0.035       0  5002.8    0.05       0  5606.3    0.16       0
Bank Sta=4996.8,5002.8
Exp/Cntr=0.3,0.1

Type RM Length L Ch R = 1,25608,282,282,282
BEGIN DESCRIPTION:
UNT166 IN CCTC 40.0
END DESCRIPTION:
XS GIS Cut Line= 2
      3556051.75     10672717.36      3555140.29     10672654.86
#Sta/Elev= 30
  4436.9  357.29  4466.4  355.59  4489.2  355.16  4509.2  353.57  4589.4  350.62
  4599.4  349.29  4729.7  344.43  4749.8  343.44  4757.9  342.42  4809.9  340.85
  4880.1  340.65  4890.1  339.13  4900.1  336.72  4906.2  338.32  4930.2  340.11
  4990.3  339.93  5000.4  330.90  5007.4  329.50  5010.1  329.00  5013.4  329.50
  5020.4  339.34  5070.5  341.00  5090.6  342.26  5120.6  345.16  5150.7  346.27
  5210.9  353.40  5261.0  356.55  5321.1  361.20  5345.9  362.33  5350.5  363.15
#Mann=3,-1,0
  4436.9    0.16       0  5007.4    0.07       0  5013.4    0.16       0
Bank Sta=5007.4,5013.4
Exp/Cntr=0.3,0.1

Type RM Length L Ch R = 1,25326,350,350,350
BEGIN DESCRIPTION:
UNT166 IN CCTC 39.0
END DESCRIPTION:
XS GIS Cut Line= 3
      3556149.61     10672260.19      3555499.61     10672410.19
      3555149.60     10672410.19
#Sta/Elev= 30
  4365.8  366.86  4417.1  365.03  4489.0  360.53  4499.2  360.76  4523.2  359.24
  4540.3  356.79  4550.5  357.20  4735.3  344.13  4742.1  342.81  4747.2  343.27
  4766.1  335.81  4784.9  334.55  4790.0  338.26  4796.8  337.60  4837.9  339.24
  4971.3  339.68  4981.6  333.16  4988.8  330.11  4991.6  329.61  4994.8  330.11
  5002.1  330.78  5008.9  337.31  5014.1  334.29  5022.6  339.49  5062.9  339.23
  5142.9  343.04  5346.7  358.96  5355.6  359.98  5362.9  361.53  5382.9  362.20
#Mann=5,-1,0
  4365.8    0.16       0  4988.8    0.07       0  4994.8    0.16       0
  5346.7    0.05       0  5355.6    0.16       0
Bank Sta=4988.8,4994.8
Exp/Cntr=0.3,0.1

Type RM Length L Ch R = 1,24976,491,491,491
BEGIN DESCRIPTION:
UNT166 IN CCTC 38.0
END DESCRIPTION:
XS GIS Cut Line= 2
      3555963.04     10671974.75      3555006.10     10672255.59
#Sta/Elev= 30
  4604.1  359.88  4659.8  357.23  4722.3  351.23  4774.4  349.21  4781.4  347.60
  4820.0  345.03  4847.4  341.04  4858.6  337.78  4868.2  337.19  4909.9  338.30
  4982.9  337.49  4992.2  335.23  5000.7  329.61  5003.5  329.11  5006.7  329.61
  5014.1  331.35  5024.5  338.84  5087.1  339.11  5108.0  338.09  5169.5  339.24
  5248.2  344.02  5274.7  344.49  5378.9  351.71  5385.5  351.17  5410.2  353.19
  5424.1  355.91  5451.8  356.34  5475.3  358.37  5545.6  361.88  5601.4  362.42
#Mann=5,-1,0
  4604.1    0.16       0  5000.7    0.07       0  5006.7    0.16       0
  5248.2    0.05       0  5475.3    0.16       0
Bank Sta=5000.7,5006.7
Exp/Cntr=0.3,0.1

Type RM Length L Ch R = 1,24485,617,617,617
BEGIN DESCRIPTION:
UNT166 IN CCTC 37.0
END DESCRIPTION:
XS GIS Cut Line= 2
      3555952.63     10671802.86      3554900.58     10671740.36
#Sta/Elev= 30
  4519.7  354.89  4582.1  351.39  4613.0  350.29  4673.0  345.22  4753.1  340.51
  4793.2  339.30  4823.3  336.80  4843.3  336.10  4873.3  337.01  4913.4  335.72
  4943.5  336.89  4982.4  336.49  4987.5  332.76  4990.6  326.51  4993.3  326.01
  4996.6  326.51  5003.6  328.31  5013.6  335.47  5023.6  336.42  5083.7  337.52
  5213.9  342.71  5264.0  346.09  5339.1  349.57  5364.2  350.84  5384.2  353.67
  5394.3  356.17  5438.0  356.43  5554.5  356.25  5564.6  359.00  5573.6  356.61
#Mann=7,-1,0
  4519.7    0.16       0  4582.1    0.05       0  4613.0    0.16       0
  4990.6    0.07       0  4996.6    0.16       0  5339.1    0.05       0
  5438.0     0.1       0
Bank Sta=4990.6,4996.6
Exp/Cntr=0.3,0.1

Type RM Length L Ch R = 1,23868,584,584,584
BEGIN DESCRIPTION:
UNT166 IN CCTC 36.0
END DESCRIPTION:
XS GIS Cut Line= 2
      3556067.19     10671672.62      3555478.71     10671219.54
#Sta/Elev= 30
  4662.5  352.56  4684.9  351.48  4790.7  344.62  4805.2  344.42  4855.0  341.14
  4894.8  339.53  4948.4  336.16  4975.5  335.73  4983.7  327.86  4990.0  324.90
  5001.5  324.35  5004.3  323.85  5007.5  324.35  5012.7  332.59  5019.0  326.64
  5025.4  333.19  5033.5  335.17  5168.5  335.17  5176.7  336.45  5203.8  337.72
  5212.0  338.85  5247.4  341.18  5253.7  342.74  5276.4  344.24  5282.7  345.45
  5300.0  346.89  5318.0  348.54  5332.5  348.74  5382.3  353.47  5405.2  354.63
#Mann=6,-1,0
  4662.5    0.16       0  4684.9    0.05       0  4894.8    0.16       0
  5001.5    0.07       0  5007.5    0.16       0  5300.0    0.05       0
Bank Sta=5001.5,5007.5
Exp/Cntr=0.3,0.1

Type RM Length L Ch R = 1,23284,787,787,787
BEGIN DESCRIPTION:
UNT166 IN CCTC 35.0
END DESCRIPTION:
XS GIS Cut Line= 3
      3556249.59     10671460.16      3556049.61     10671060.19
      3555699.58     10670910.17
#Sta/Elev= 30
  4580.0  344.17  4611.1  342.22  4789.7  334.69  4803.6  334.95  4848.3  332.94
  4901.4  332.48  4946.1  333.68  4960.1  330.24  4968.5  330.66  4974.1  332.75
  4990.8  327.94  4996.4  329.13  5001.8  323.11  5004.6  322.61  5007.8  323.11
  5013.2  329.93  5018.8  328.94  5024.4  331.92  5059.8  332.22  5094.3  330.19
  5112.4  330.25  5117.8  333.19  5125.1  333.94  5179.5  335.00  5271.3  340.36
  5299.2  341.60  5317.3  343.32  5322.7  344.71  5398.9  350.78  5408.0  350.82
#Mann=6,-1,0
  4580.0    0.16       0  4611.1    0.05       0  4789.7    0.16       0
  5001.8    0.07       0  5007.8    0.16       0  5271.3    0.05       0
Bank Sta=5001.8,5007.8
Exp/Cntr=0.3,0.1

Type RM Length L Ch R = 1,22497,104,104,104
BEGIN DESCRIPTION:
UNT166 IN CCTC 34.0
END DESCRIPTION:
XS GIS Cut Line= 3
      3556981.63     10671278.22      3556460.83     10670889.36
      3556016.39     10670656.73
#Sta/Elev= 30
  4402.0  354.76  4699.0  340.60  4770.9  336.76  4866.3  331.54  4909.2  332.53
  4923.8  328.21  4930.1  330.98  4938.9  329.27  4943.9  329.16  4953.0  328.73
  4959.3  325.61  4973.9  330.15  4980.1  324.38  4988.5  324.63  4991.7  321.60
  4994.4  321.10  4997.7  321.60  5016.0  322.38  5030.1  330.01  5058.2  329.53
  5065.6  331.26  5142.6  332.50  5148.2  334.12  5208.8  333.33  5363.3  339.01
  5451.6  339.50  5490.1  343.51  5534.2  346.13  5539.8  344.65  5553.6  346.61
#Mann=8,-1,0
  4402.0    0.05       0  4699.0    0.12       0  4770.9    0.05       0
  4938.9    0.12       0  4943.9    0.08       0  4991.7    0.07       0
  4997.7    0.08       0  5058.2    0.05       0
Bank Sta=4991.7,4997.7
Exp/Cntr=0.3,0.1

Type RM Length L Ch R = 1,22393,605,605,605
BEGIN DESCRIPTION:
UNT166 IN CCTC 33.0
END DESCRIPTION:
XS GIS Cut Line= 3
      3557061.51     10671229.63      3556495.56     10670826.86
      3556075.38     10670580.32
#Sta/Elev= 30
  4426.8  355.81  4491.4  352.95  4527.3  350.23  4550.5  350.28  4556.6  348.99
  4621.8  347.00  4686.9  342.63  4736.0  342.16  4749.6  340.71  4829.6  337.72
  4936.5  331.60  4951.3  332.29  4980.8  329.52  4993.7  325.05  4998.7  321.34
  5001.5  320.84  5004.7  321.34  5007.9  322.22  5016.5  327.97  5030.5  330.71
  5048.6  330.65  5072.1  329.73  5087.8  331.02  5129.4  330.47  5164.4  331.33
  5271.8  332.45  5275.9  332.53  5453.0  341.05  5536.6  346.45  5608.6  349.93
#Mann=9,-1,0
  4426.8    0.05       0  4998.7    0.04       0  5004.7    0.05       0
  5048.6    0.08       0  5072.1    0.12       0  5164.4    0.05       0
  5271.8    0.12       0  5275.9    0.16       0  5536.6    0.05       0
Bank Sta=4998.7,5004.7
Exp/Cntr=0.3,0.1

Type RM Length L Ch R = 1,21788,416,416,416
BEGIN DESCRIPTION:
UNT166 IN CCTC 32.0
END DESCRIPTION:
XS GIS Cut Line= 2
      3557218.29     10670714.33      3556410.97     10670297.65
#Sta/Elev= 30
  4430.2  346.07  4558.6  337.48  4597.3  336.22  4647.3  333.09  4721.3  328.85
  4766.3  327.96  4856.3  329.74  4878.8  326.13  4885.3  326.26  4891.0  328.19
  4901.4  329.32  4935.3  327.96  4957.6  329.47  4974.0  328.83  4980.1  328.45
  4990.5  321.70  4993.1  318.53  4995.9  318.03  4999.1  318.53  5002.6  319.24
  5012.6  326.47  5070.2  335.17  5079.1  335.41  5092.7  337.95  5174.5  344.13
  5212.0  344.95  5217.7  346.34  5250.2  347.24  5262.0  348.84  5338.7  352.91
#Mann=5,-1,0
  4430.2    0.16       0  4647.3    0.12       0  4993.1    0.07       0
  4999.1    0.12       0  5174.5    0.16       0
Bank Sta=4993.1,4999.1
Exp/Cntr=0.3,0.1

Type RM Length L Ch R = 1,21372,994,994,994
BEGIN DESCRIPTION:
UNT166 IN CCTC 31.0
END DESCRIPTION:
XS GIS Cut Line= 2
      3557374.50     10670620.55      3556614.39     10669912.50
#Sta/Elev= 30
  4485.0  347.22  4552.4  342.46  4609.0  339.90  4623.2  338.11  4637.4  337.94
  4700.9  332.68  4715.1  332.50  4792.7  327.43  4821.6  326.97  4856.8  326.95
  4870.9  325.13  4920.3  327.78  4970.0  327.80  4991.1  320.56  4994.9  317.66
  4997.7  317.16  5000.9  317.66  5012.1  323.36  5019.4  328.53  5026.3  329.43
  5097.1  332.71  5195.0  339.01  5224.6  341.29  5291.6  344.20  5323.8  346.78
  5330.7  346.49  5338.0  347.60  5472.3  354.16  5486.5  355.80  5523.8  357.80
#Mann=6,-1,0
  4485.0    0.16       0  4821.6    0.12       0  4994.9    0.07       0
  5000.9    0.12       0  5195.0    0.16       0  5291.6    0.05       0
Bank Sta=4994.9,5000.9
Exp/Cntr=0.3,0.1

Type RM Length L Ch R = 1,20378,813,813,813
BEGIN DESCRIPTION:
UNT166 IN CCTC 30.0
END DESCRIPTION:
XS GIS Cut Line= 2
      3557856.68     10670229.65      3556945.62     10669744.67
#Sta/Elev= 30
  4411.9  343.60  4431.2  341.74  4476.6  339.51  4511.4  338.99  4527.7  337.38
  4565.9  335.51  4724.9  329.74  4873.5  325.39  4955.7  326.05  4977.7  323.77
  4986.3  319.86  4999.4  315.29  5006.0  314.74  5008.7  314.24  5012.0  314.74
  5016.0  317.08  5021.6  322.53  5031.7  319.17  5043.6  324.71  5054.2  323.60
  5059.9  326.02  5156.3  328.47  5213.7  331.16  5230.0  333.10  5252.0  334.03
  5273.9  336.32  5310.8  338.73  5339.8  340.28  5438.4  349.05  5444.0  350.40
#Mann=6,-1,0
  4411.9    0.16       0  4724.9    0.12       0  4999.4    0.16       0
  5006.0    0.07       0  5012.0    0.16       0  5310.8    0.05       0
Bank Sta=5006,5012
Exp/Cntr=0.3,0.1

Type RM Length L Ch R = 1,19565,617,617,617
BEGIN DESCRIPTION:
UNT166 IN CCTC 29.0
END DESCRIPTION:
XS GIS Cut Line= 3
      3557949.64     10669910.21      3557599.61     10669660.19
      3557199.64     10669260.22
#Sta/Elev= 30
  4557.6  342.30  4606.8  339.49  4636.3  335.46  4665.8  334.38  4716.2  330.78
  4722.3  330.99  4781.6  327.67  4864.9  324.95  4901.7  325.09  4923.9  324.20
  4959.5  324.63  4974.2  324.11  4980.4  321.20  4984.7  317.39  4991.3  317.39
  4998.9  311.12  5001.6  310.62  5004.9  311.12  5016.0  314.25  5030.2  324.00
  5058.5  322.73  5100.9  323.14  5190.2  325.46  5228.2  326.25  5270.6  328.35
  5284.7  328.50  5341.3  331.82  5383.7  333.38  5468.6  341.16  5553.4  346.72
#Mann=5,-1,0
  4557.6    0.16       0  4781.6    0.12       0  4998.9    0.07       0
  5004.9    0.12       0  5190.2    0.16       0
Bank Sta=4998.9,5004.9
Exp/Cntr=0.3,0.1

Type RM Length L Ch R = 1,18948,616,616,616
BEGIN DESCRIPTION:
UNT166 IN CCTC 28.0
END DESCRIPTION:
XS GIS Cut Line= 3
      3558049.60     10669710.17      3557799.61     10669310.19
      3557799.61     10668910.17
#Sta/Elev= 30
  4545.7  334.69  4574.6  333.93  4720.8  324.00  4765.0  323.53  4836.4  321.16
  4958.4  322.79  4982.0  317.50  4991.4  310.82  4994.1  310.32  4997.4  310.82
  5003.8  312.50  5009.7  317.49  5014.4  319.44  5027.4  317.76  5037.4  313.56
  5047.4  314.29  5057.4  323.68  5077.4  321.39  5087.4  321.82  5127.4  325.65
  5137.4  327.83  5147.4  327.59  5167.4  322.99  5190.4  321.91  5217.4  323.87
  5237.4  328.21  5257.4  329.08  5287.4  332.69  5297.4  332.39  5417.4  343.22
#Mann=5,-1,0
  4545.7    0.16       0  4765.0    0.12       0  4991.4    0.07       0
  4997.4    0.12       0  5190.4    0.16       0
Bank Sta=4991.4,4997.4
Exp/Cntr=0.3,0.1

Type RM Length L Ch R = 1,18332,557,557,557
BEGIN DESCRIPTION:
UNT166 IN CCTC 27.0
END DESCRIPTION:
XS GIS Cut Line= 2
      3558166.19     10669714.28      3558254.52     10668784.26
#Sta/Elev= 30
  4618.1  337.22  4700.2  331.11  4782.9  325.84  4843.2  323.72  4883.4  320.41
  4903.1  320.22  4953.7  321.01  4963.7  318.86  4983.8  318.65  5000.9  309.25
  5003.7  308.75  5006.9  309.25  5021.7  316.77  5034.1  320.56  5044.1  321.83
  5074.2  321.56  5084.3  318.63  5094.3  318.78  5104.4  321.51  5129.8  323.22
  5194.8  323.51  5258.0  325.53  5285.2  328.34  5305.3  328.41  5355.5  335.35
  5385.6  336.74  5405.7  339.93  5425.8  339.64  5506.2  346.48  5552.3  348.23
#Mann=6,-1,0
  4618.1    0.05       0  4700.2    0.16       0  4903.1    0.12       0
  5000.9    0.07       0  5006.9    0.12       0  5258.0    0.16       0
Bank Sta=5000.9,5006.9
Exp/Cntr=0.3,0.1

Type RM Length L Ch R = 1,17775,780,780,780
BEGIN DESCRIPTION:
UNT166 IN CCTC 26.0
END DESCRIPTION:
XS GIS Cut Line= 3
      3558299.59     10669710.21      3558549.61     10669310.19
      3558549.61     10668910.22
#Sta/Elev= 30
  4518.7  334.54  4599.5  328.43  4620.7  328.28  4642.0  325.90  4715.1  322.04
  4788.2  320.55  4824.7  321.18  4856.6  319.74  4946.2  320.22  4955.0  319.03
  4961.5  311.93  4967.4  313.68  4976.9  311.01  4982.8  312.46  4987.5  309.85
  4992.9  309.85  4997.4  308.34  5000.2  307.84  5003.4  308.34  5010.4  310.30
  5020.4  318.30  5030.4  318.17  5070.4  321.20  5190.4  324.03  5230.4  329.01
  5243.2  329.29  5310.4  335.22  5360.4  338.39  5370.4  340.03  5390.4  340.38
#Mann=5,-1,0
  4518.7    0.16       0  4856.6    0.12       0  4997.4    0.07       0
  5003.4    0.12       0  5243.2    0.16       0
Bank Sta=4997.4,5003.4
Exp/Cntr=0.3,0.1

Type RM Length L Ch R = 1,16995,328,328,328
BEGIN DESCRIPTION:
UNT166 IN CCTC 25.0
END DESCRIPTION:
XS GIS Cut Line= 4
      3558538.21     10669917.40      3559111.15     10669452.98
      3559141.53     10669201.24      3558655.43     10668849.68
#Sta/Elev= 30
  4166.3  329.63  4200.9  328.50  4278.8  322.57  4570.2  319.28  4599.0  317.19
  4605.8  319.05  4627.7  319.71  4916.7  317.89  4926.8  316.86  4932.3  314.19
  4937.3  315.59  4946.9  312.49  4957.0  316.01  4967.1  317.38  4977.1  316.99
  5004.4  306.77  5007.1  306.27  5010.4  306.77  5014.3  309.24  5019.3  309.80
  5027.5  318.88  5138.3  317.40  5166.8  318.89  5353.2  318.25  5440.8  321.68
  5596.1  330.13  5690.4  333.54  5696.7  332.71  5711.4  334.70  5757.3  336.77
#Mann=5,-1,0
  4166.3    0.16       0  4278.8    0.12       0  5004.4    0.07       0
  5010.4    0.12       0  5440.8    0.16       0
Bank Sta=5004.4,5010.4
Exp/Cntr=0.3,0.1

Type RM Length L Ch R = 1,16667,486,486,486
BEGIN DESCRIPTION:
UNT166 IN CCTC 24.0
END DESCRIPTION:
XS GIS Cut Line= 3
      3559631.98     10669817.55      3559228.34     10669066.69
      3558889.80     10668702.11
#Sta/Elev= 30
  4276.7  341.95  4351.6  340.75  4401.1  337.74  4439.2  337.81  4444.9  336.81
  4477.4  336.32  4521.2  334.28  4526.9  333.19  4543.1  333.09  4548.8  331.81
  4682.4  322.52  4794.7  317.54  4800.4  318.33  4819.6  317.88  4926.2  318.38
  4942.4  316.96  4970.0  317.32  4977.6  316.55  4986.3  312.43  4997.3  304.40
  5000.1  303.90  5003.3  304.40  5008.2  308.15  5030.1  317.92  5052.0  318.02
  5079.8  316.59  5334.3  318.14  5361.9  319.07  5449.9  322.48  5626.7  329.80
#Mann=7,-1,0
  4276.7    0.16       0  4819.6    0.12       0  4997.3    0.07       0
  5003.3    0.12       0  5334.3    0.16       0  5361.9    0.12       0
  5449.9    0.16       0
Bank Sta=4997.3,5003.3
Exp/Cntr=0.3,0.1

Type RM Length L Ch R = 1,16181,667,667,667
BEGIN DESCRIPTION:
UNT166 IN CCTC 23.0
END DESCRIPTION:
XS GIS Cut Line= 2
      3559710.11     10669513.74      3559285.42     10668313.35
#Sta/Elev= 30
  4463.0  331.87  4475.8  330.96  4488.0  331.59  4530.4  327.62  4686.8  319.04
  4777.0  317.51  4836.0  316.07  4872.2  316.88  4891.1  315.06  4897.8  315.54
  4903.1  313.43  4922.9  314.60  4934.0  312.08  4954.3  312.38  4975.9  314.51
  4985.2  306.86  4990.5  306.19  4994.1  303.45  4996.9  302.95  5000.1  303.45
  5007.7  308.22  5016.1  311.45  5021.4  310.76  5029.0  315.99  5039.6  316.90
  5127.0  315.79  5319.8  316.86  5357.8  318.62  5407.2  318.26  5736.3  324.83
#Mann=5,-1,0
  4463.0    0.16       0  4777.0    0.12       0  4994.1    0.07       0
  5000.1    0.12       0  5127.0    0.16       0
Bank Sta=4994.1,5000.1
Exp/Cntr=0.3,0.1

Type RM Length L Ch R = 1,15514,561,561,561
BEGIN DESCRIPTION:
UNT166 IN CCTC 22.0
END DESCRIPTION:
XS GIS Cut Line= 3
      3560256.95     10669196.87      3559888.06     10668914.78
      3559575.56     10668207.31
#Sta/Elev= 30
  4430.9  335.89  4548.0  327.28  4797.4  316.99  4833.1  312.96  4847.3  309.91
  4855.5  315.00  4861.8  313.42  4876.3  315.52  4965.9  315.88  4980.2  314.21
  4987.8  311.55  4998.0  302.29  5006.6  302.17  5009.4  301.67  5012.6  302.17
  5020.6  309.49  5026.8  311.87  5042.4  313.66  5073.4  312.59  5078.9  314.09
  5096.7  309.98  5102.2  310.04  5108.0  313.92  5118.9  315.10  5192.1  313.84
  5369.5  315.15  5450.3  317.47  5534.4  323.62  5543.6  325.50  5668.7  331.55
#Mann=5,-1,0
  4430.9    0.16       0  4833.1    0.12       0  5006.6    0.07       0
  5012.6    0.12       0  5192.1    0.16       0
Bank Sta=5006.6,5012.6
Exp/Cntr=0.3,0.1

Type RM Length L Ch R = 1,14953,769,769,769
BEGIN DESCRIPTION:
UNT166 IN CCTC 21.0
END DESCRIPTION:
XS GIS Cut Line= 3
      3560449.58     10668860.16      3560099.61     10668560.19
      3559599.57     10668160.16
#Sta/Elev= 30
  4512.2  343.37  4618.1  335.65  4640.0  332.89  4816.7  320.06  4831.0  319.92
  4867.2  313.84  4880.9  312.81  4945.1  313.90  4978.6  311.84  4986.7  311.09
  4994.7  302.95  5006.2  301.39  5008.9  300.89  5012.2  301.39  5015.6  306.98
  5023.6  313.15  5030.0  314.71  5050.8  312.06  5058.8  312.24  5065.2  310.32
  5087.6  313.35  5129.2  313.30  5158.0  315.27  5186.8  314.13  5206.8  314.80
  5279.7  314.58  5350.1  316.07  5414.2  319.35  5556.6  331.13  5613.5  332.68
#Mann=5,-1,0
  4512.2    0.16       0  4978.6    0.12       0  5006.2    0.07       0
  5012.2    0.12       0  5206.8    0.16       0
Bank Sta=5006.2,5012.2
Exp/Cntr=0.3,0.1

Type RM Length L Ch R = 1,14184,870,870,870
BEGIN DESCRIPTION:
UNT166 IN CCTC 20.0
END DESCRIPTION:
XS GIS Cut Line= 3
      3560702.31     10668883.74      3560563.41     10668189.26
      3560188.39     10667640.61
#Sta/Elev= 30
  4175.3  343.90  4240.1  340.70  4301.3  336.41  4311.5  334.92  4316.6  335.32
  4331.9  333.65  4433.9  328.03  4444.1  326.77  4464.4  325.60  4474.7  326.22
  4484.9  324.25  4651.5  312.78  4719.4  310.58  4950.7  312.86  4979.3  311.22
  4986.5  308.76  4992.6  302.58  5004.5  300.43  5007.3  299.93  5010.5  300.43
  5015.6  305.34  5028.5  312.21  5074.8  313.30  5130.1  314.47  5195.8  318.30
  5237.8  319.64  5294.6  323.73  5381.3  328.39  5411.2  329.14  5548.1  337.55
#Mann=5,-1,0
  4175.3    0.16       0  4651.5    0.12       0  5004.5    0.07       0
  5010.5    0.12       0  5074.8    0.05       0
Bank Sta=5004.5,5010.5
Exp/Cntr=0.3,0.1

Type RM Length L Ch R = 1,13314,368,368,368
BEGIN DESCRIPTION:
UNT166 IN CCTC 19.0
END DESCRIPTION:
XS GIS Cut Line= 3
      3560980.08     10669404.51      3561112.02     10668182.32
      3560286.43     10667384.48
#Sta/Elev= 30
  3979.6  339.99  4112.3  341.43  4154.9  339.40  4392.9  334.56  4581.6  326.62
  4627.7  325.96  4969.6  311.47  4979.7  309.89  4989.8  304.73  4996.8  298.50
  4999.6  298.00  5002.8  298.50  5009.9  305.33  5019.9  306.48  5040.0  305.43
  5060.2  309.14  5090.3  310.52  5160.7  309.55  5516.3  311.24  5601.2  310.48
  5777.9  313.45  5905.2  324.13  5954.6  326.58  5961.8  328.43  5968.8  327.65
  5982.9  330.12  5990.1  328.71  6053.7  331.69  6244.6  337.03  6357.0  343.66
#Mann=3,-1,0
  3979.6    0.05       0  4996.8    0.03       0  5002.8    0.05       0
Bank Sta=4996.8,5002.8
Exp/Cntr=0.3,0.1

Type RM Length L Ch R = 1,12946,652,652,652
BEGIN DESCRIPTION:
UNT166 IN CCTC 18.0
END DESCRIPTION:
XS GIS Cut Line= 2
      3562028.66     10669050.34      3560495.03     10667294.65
#Sta/Elev= 30
  3856.8  336.42  4069.3  329.34  4337.9  314.13  4430.0  310.87  4538.2  310.72
  4636.0  310.92  4756.5  308.45  4938.5  309.27  4975.8  308.38  4983.4  300.70
  4990.0  301.83  4997.6  298.11  5008.9  297.47  5011.6  296.97  5014.9  297.47
  5018.5  301.95  5032.8  308.48  5047.0  309.26  5515.0  311.12  5550.1  312.40
  5556.7  314.43  5585.2  316.73  5621.3  317.21  5649.5  316.49  5656.4  314.18
  5705.8  313.73  5776.9  315.69  5840.6  320.64  5906.2  323.89  6188.0  338.64
#Mann=7,-1,0
  3856.8    0.16       0  4538.2    0.12       0  4938.5    0.05       0
  5008.9    0.03       0  5014.9    0.05       0  5840.6    0.16       0
  5906.2    0.05       0
Bank Sta=5008.9,5014.9
Exp/Cntr=0.3,0.1

Type RM Length L Ch R = 1,12294,871,871,871
BEGIN DESCRIPTION:
UNT166 IN CCTC 17.0
END DESCRIPTION:
XS GIS Cut Line= 3
      3562013.06     10668728.15      3561575.56     10668103.15
      3561436.67     10667200.38
#Sta/Elev= 30
  4097.5  326.41  4249.7  319.56  4417.2  314.79  4567.7  308.94  4666.4  307.68
  4822.3  308.47  4964.6  309.09  4974.7  306.61  4996.1  296.57  4998.8  296.07
  5002.1  296.57  5015.2  303.96  5025.3  307.24  5055.6  308.23  5099.3  307.49
  5130.6  307.43  5146.7  303.57  5156.8  304.24  5166.9  307.23  5177.0  307.67
  5278.2  309.44  5479.3  316.15  5511.3  317.94  5588.4  321.42  5622.2  321.73
  5651.7  324.16  5656.7  323.39  5693.0  325.38  5743.6  325.50  5773.8  327.00
#Mann=9,-1,0
  4097.5    0.16       0  4417.2    0.12       0  4567.7    0.16       0
  4822.3    0.12       0  4996.1    0.07       0  5002.1    0.12       0
  5099.3    0.05       0  5479.3    0.16       0  5511.3    0.05       0
Bank Sta=4996.1,5002.1
Exp/Cntr=0.3,0.1

Type RM Length L Ch R = 1,11423,760,760,760
BEGIN DESCRIPTION:
UNT166 IN CCTC 16.0
END DESCRIPTION:
XS GIS Cut Line= 2
      3562096.39     10668880.91      3562096.39     10667068.41
#Sta/Elev= 30
  4314.7  331.86  4465.4  327.79  4485.4  325.53  4625.4  320.18  4645.4  318.29
  4665.4  318.66  4815.4  308.39  4855.4  306.70  4915.4  305.78  4932.5  307.22
  4965.4  307.51  4985.4  296.60  4992.4  295.34  4995.2  294.84  4998.4  295.34
  5005.4  297.03  5025.4  305.81  5035.4  306.47  5105.4  307.40  5145.4  306.06
  5285.4  305.68  5395.5  311.27  5553.0  320.13  5595.4  323.06  5835.4  329.34
  5885.4  331.94  5945.4  333.09  5955.4  334.39  6086.0  335.98  6127.2  336.51
#Mann=7,-1,0
  4314.7    0.16       0  4932.5    0.12       0  4992.4    0.07       0
  4998.4    0.12       0  5395.5    0.05       0  5553.0    0.16       0
  6086.0    0.05       0
Bank Sta=4992.4,4998.4
Exp/Cntr=0.3,0.1

Type RM Length L Ch R = 1,10663,512,512,512
BEGIN DESCRIPTION:
UNT166 IN CCTC 15.0
END DESCRIPTION:
XS GIS Cut Line= 3
      3562381.11     10668860.12      3562506.12     10668269.82
      3562506.12     10667444.31
#Sta/Elev= 30
  4517.3  331.22  4527.5  329.78  4619.5  326.35  4639.9  324.12  4711.4  321.21
  4742.1  318.47  4834.1  313.15  4864.8  312.61  4946.5  307.62  4956.8  305.59
  4977.2  304.84  4987.4  302.01  4994.7  293.73  4997.4  293.23  5000.7  293.73
  5007.9  298.93  5014.9  300.70  5028.3  306.22  5044.3  306.19  5079.4  305.35
  5114.3  306.65  5170.3  305.09  5180.3  305.89  5190.3  305.27  5200.3  306.53
  5320.3  305.34  5372.9  306.20  5520.3  310.68  5699.2  319.77  5946.2  333.72
#Mann=6,-1,0
  4517.3    0.16       0  4994.7    0.07       0  5000.7    0.16       0
  5044.3    0.12       0  5372.9    0.05       0  5699.2    0.16       0
Bank Sta=4994.7,5000.7
Exp/Cntr=0.3,0.1

Type RM Length L Ch R = 1,10151,485,485,485
BEGIN DESCRIPTION:
UNT166 IN CCTC 13.0
END DESCRIPTION:
XS GIS Cut Line= 3
      3562949.61     10668960.20      3562749.61     10668160.19
      3562699.61     10667560.20
#Sta/Elev= 30
  4173.6  330.08  4232.9  327.97  4297.3  323.98  4328.2  321.06  4397.8  318.28
  4480.3  312.67  4544.7  309.79  4627.2  307.22  4687.8  307.24  4732.8  306.48
  4774.0  304.13  4833.3  304.83  4884.8  303.81  4967.3  305.05  4975.0  300.99
  4980.2  304.32  4992.7  292.53  4995.4  292.03  4998.7  292.53  5008.3  294.91
  5018.3  303.64  5028.3  305.29  5048.4  303.93  5098.7  304.64  5148.8  305.71
  5239.1  309.93  5269.2  312.61  5339.4  316.28  5520.0  330.10  5600.3  333.22
#Mann=5,-1,0
  4173.6    0.16       0  4687.8    0.12       0  4992.7    0.07       0
  4998.7    0.12       0  5098.7    0.16       0
Bank Sta=4992.7,4998.7
Exp/Cntr=0.3,0.1

Type RM Length L Ch R = 1,9666,463,463,463
BEGIN DESCRIPTION:
UNT166 IN CCTC 12.0
END DESCRIPTION:
XS GIS Cut Line= 3
      3563049.60     10668910.23      3563149.61     10668110.19
      3563099.61     10667710.17
#Sta/Elev= 30
  4178.7  332.73  4420.6  314.96  4440.8  314.85  4516.7  310.22  4539.0  308.37
  4612.1  306.19  4632.2  304.44  4682.6  302.63  4833.8  302.91  4894.3  304.87
  4964.8  304.55  4974.9  303.51  4982.5  296.98  4987.5  296.98  4992.0  292.38
  4994.8  291.88  4998.0  292.38  5005.1  296.82  5015.2  299.91  5019.4  302.49
  5022.8  304.58  5027.8  302.91  5035.4  304.65  5065.6  304.37  5126.1  307.89
  5156.3  310.76  5226.8  313.92  5269.7  317.12  5277.2  319.14  5388.1  326.35
#Mann=5,-1,0
  4178.7    0.16       0  4516.7    0.12       0  4992.0    0.07       0
  4998.0    0.12       0  5019.4    0.16       0
Bank Sta=4992,4998
Exp/Cntr=0.3,0.1

Type RM Length L Ch R = 1,9203,168,168,168
BEGIN DESCRIPTION:
UNT166 IN CCTC 11.0
END DESCRIPTION:
XS GIS Cut Line= 3
      3563049.63     10669010.15      3563549.61     10668010.19
      3563499.61     10667610.19
#Sta/Elev= 30
  3855.1  337.00  3936.1  334.21  3997.6  329.41  4056.3  326.63  4257.5  313.55
  4288.3  312.98  4419.5  306.49  4511.9  302.58  4517.5  303.26  4593.0  301.28
  4713.1  302.86  4718.7  301.83  4757.9  303.56  4899.0  302.53  4942.3  302.37
  4950.7  303.25  4974.4  301.47  4983.2  299.73  4990.2  291.86  4993.0  291.36
  4996.2  291.86  5003.3  292.79  5010.9  300.85  5015.9  299.69  5023.5  305.58
  5053.9  306.89  5177.2  316.78  5235.1  320.33  5265.3  323.73  5376.2  329.37
#Mann=7,-1,0
  3855.1    0.16       0  4419.5    0.12       0  4899.0    0.16       0
  4974.4    0.12       0  4990.2    0.07       0  4996.2    0.12       0
  5053.9    0.16       0
Bank Sta=4990.2,4996.2
Exp/Cntr=0.3,0.1

Type RM Length L Ch R = 1,9035,1166,1166,1166
BEGIN DESCRIPTION:
UNT166 IN CCTC 10.0
END DESCRIPTION:
XS GIS Cut Line= 2
      3563359.91     10668902.15      3563936.32     10667409.05
#Sta/Elev= 30
  4114.6  325.76  4148.9  325.10  4154.8  324.06  4184.8  323.44  4191.7  322.04
  4353.8  315.43  4408.4  312.20  4416.8  310.90  4592.0  301.74  4642.0  300.15
  4856.3  302.02  4874.9  300.49  4959.4  302.96  4974.2  302.54  4984.0  299.26
  4989.4  293.20  4992.7  291.76  4995.4  291.26  4998.7  291.76  5006.4  294.24
  5019.3  303.43  5135.0  301.72  5262.2  305.19  5322.1  305.18  5455.9  307.62
  5515.8  310.54  5521.1  309.65  5545.7  309.82  5619.0  311.78  5715.1  313.88
#Mann=5,-1,0
  4114.6    0.16       0  4592.0    0.12       0  4992.7    0.07       0
  4998.7    0.12       0  5619.0    0.16       0
Bank Sta=4992.7,4998.7
Exp/Cntr=0.3,0.1

Type RM Length L Ch R = 1,7869,437,437,437
BEGIN DESCRIPTION:
UNT166 IN CCTC 9.0
END DESCRIPTION:
XS GIS Cut Line= 3
      3563561.29     10669006.31      3564283.54     10668388.23
      3564359.92     10667395.18
#Sta/Elev= 30
  3799.7  322.91  3902.6  321.64  3987.2  318.13  4155.7  304.00  4192.4  301.67
  4319.8  301.27  4335.3  300.92  4497.6  300.57  4561.3  298.36  4568.9  299.79
  4589.8  300.06  4696.3  299.66  4704.0  298.25  4724.8  300.25  4858.7  301.04
  4868.7  300.65  4878.7  297.44  4888.8  297.29  4969.0  300.77  4979.0  299.23
  4986.1  290.22  4988.8  289.72  4992.1  290.22  4999.1  291.43  5009.1  297.60
  5019.1  300.84  5188.4  299.56  5274.6  302.70  5392.1  305.97  5746.3  317.77
#Mann=9,-1,0
  3799.7    0.16       0  4155.7    0.12       0  4319.8    0.16       0
  4335.3    0.12       0  4986.1    0.07       0  4992.1    0.12       0
  5188.4    0.16       0  5274.6    0.12       0  5392.1    0.16       0
Bank Sta=4986.1,4992.1
Exp/Cntr=0.3,0.1

Type RM Length L Ch R = 1,7432,1214,1214,1214
BEGIN DESCRIPTION:
UNT166 IN CCTC 8.0
END DESCRIPTION:
XS GIS Cut Line= 3
      3564700.20     10669228.49      3564568.26     10668186.85
      3564665.42     10667374.81
#Sta/Elev= 30
  3806.3  332.68  3885.2  333.64  3993.5  327.21  4163.7  316.03  4399.3  300.36
  4449.7  300.43  4486.2  294.27  4491.2  291.27  4510.2  294.01  4520.3  300.28
  4550.5  298.59  4661.4  297.57  4801.6  298.44  4852.1  299.95  4909.0  298.85
  4953.6  300.97  4973.8  300.13  4983.8  295.76  4993.4  289.34  4996.2  288.84
  4999.4  289.34  5004.0  289.78  5014.0  300.50  5054.3  299.28  5131.7  301.50
  5243.5  306.38  5346.4  312.56  5385.8  312.71  5500.7  314.67  5674.1  322.59
#Mann=7,-1,0
  3806.3    0.12       0  3993.5    0.16       0  4163.7    0.12       0
  4993.4    0.07       0  4999.4    0.12       0  5131.7    0.16       0
  5385.8    0.05       0
Bank Sta=4993.4,4999.4
Exp/Cntr=0.3,0.1

Type RM Length L Ch R = 1,6218,641,641,641
BEGIN DESCRIPTION:
UNT166 IN CCTC 7.0
END DESCRIPTION:
XS GIS Cut Line= 3
      3564846.04     10669284.07      3565172.42     10668554.90
      3564943.26     10667395.21
#Sta/Elev= 30
  3823.4  323.32  3901.7  321.38  3988.9  316.87  4002.9  315.00  4178.2  307.95
  4349.4  297.18  4405.1  295.46  4637.3  294.34  4785.0  296.18  4800.4  297.50
  4821.6  295.56  4851.3  296.03  4892.1  298.81  4912.5  295.64  4970.3  298.62
  4975.4  298.34  4983.9  294.07  5001.2  288.55  5004.0  288.05  5007.2  288.55
  5014.4  289.10  5034.8  297.78  5045.0  298.44  5167.3  296.62  5242.7  297.41
  5334.4  301.13  5422.2  308.40  5590.7  319.03  5707.6  323.40  5804.4  324.83
#Mann=7,-1,0
  3823.4    0.16       0  3901.7    0.12       0  4349.4    0.05       0
  4785.0    0.12       0  5001.2    0.07       0  5007.2    0.12       0
  5242.7    0.05       0
Bank Sta=5001.2,5007.2
Exp/Cntr=0.3,0.1

Type RM Length L Ch R = 1,5577,768,768,768
BEGIN DESCRIPTION:
UNT166 IN CCTC 5.0
END DESCRIPTION:
XS GIS Cut Line= 3
      3564991.86     10669575.74      3565714.09     10668263.23
      3565137.72     10667367.43
#Sta/Elev= 30
  3254.4  322.35  3426.1  312.95  3509.6  309.88  3680.5  304.41  3808.6  299.83
  3946.6  297.21  4110.8  297.42  4390.7  294.32  4420.5  292.81  4589.0  293.99
  4744.6  292.26  4793.1  293.54  4923.2  292.54  4946.4  293.50  4968.8  298.26
  4972.3  296.90  4989.9  288.43  5008.0  288.04  5010.8  287.54  5014.0  288.04
  5017.7  296.66  5172.9  297.07  5265.3  296.63  5416.5  306.53  5445.8  310.14
  5540.6  315.48  5567.7  318.43  5619.2  319.62  5640.3  322.09  5817.7  327.27
#Mann=8,-1,0
  3254.4    0.05       0  3509.6    0.16       0  3680.5    0.12       0
  3946.6    0.05       0  4972.3    0.12       0  5008.0    0.07       0
  5014.0    0.12       0  5172.9    0.05       0
Bank Sta=5008,5014
Exp/Cntr=0.3,0.1

Type RM Length L Ch R = 1,4809,617,617,617
BEGIN DESCRIPTION:
UNT166 IN CCTC 4.0
END DESCRIPTION:
XS GIS Cut Line= 3
      3566001.42     10669765.81      3566120.78     10667823.56
      3565415.46     10666738.46
#Sta/Elev= 30
  2651.7  327.98  2660.3  323.76  2687.4  313.65  2727.5  309.65  2871.5  310.57
  3043.9  305.28  3128.2  302.18  3138.2  300.83  3148.3  295.50  3153.0  297.08
  3168.3  301.48  3218.4  297.80  3458.8  297.88  3749.4  303.74  3889.7  302.53
  4006.4  295.39  4230.3  290.47  4908.6  295.02  4970.7  295.56  4991.8  292.94
  5003.9  287.36  5006.6  286.86  5009.9  287.36  5018.4  291.95  5028.0  295.77
  5105.5  293.30  5189.6  293.34  5438.6  299.55  5816.1  316.01  5891.8  321.64
#Mann=11,-1,0
  2651.7    0.05       0  2660.3    0.16       0  2871.5    0.12       0
  3043.9    0.16       0  3153.0    0.05       0  4908.6    0.12       0
  5003.9    0.07       0  5009.9    0.12       0  5018.4    0.05       0
  5105.5    0.16       0  5189.6    0.05       0
Bank Sta=5003.9,5009.9
Exp/Cntr=0.3,0.1

Type RM Length L Ch R = 1,4192,1105,1105,1105
BEGIN DESCRIPTION:
UNT166 IN CCTC 3.0
END DESCRIPTION:
XS GIS Cut Line= 3
      3566283.54     10669733.24      3566533.10     10667454.64
      3566034.28     10666500.38
#Sta/Elev= 30
  2456.7  322.86  2590.5  315.68  2852.1  295.92  2934.5  292.88  3010.9  292.94
  3445.6  288.93  3878.2  291.38  4059.3  291.50  4117.2  289.67  4578.2  290.84
  4958.8  294.03  4984.2  294.74  5003.3  287.67  5006.0  287.17  5009.3  287.67
  5013.5  288.53  5022.7  295.01  5148.9  295.98  5243.5  303.71  5282.0  310.19
  5287.6  308.49  5295.6  309.36  5304.1  312.91  5348.1  315.46  5439.9  319.97
  5461.0  321.13  5574.0  327.15  5638.5  329.82  5706.3  332.72  5825.7  334.05
#Mann=12,-1,0
  2456.7    0.16       0  2934.5    0.12       0  3010.9    0.05       0
  4958.8    0.12       0  5003.3    0.07       0  5009.3    0.12       0
  5348.1    0.05       0  5439.9    0.16       0  5461.0    0.05       0
  5574.0    0.16       0  5638.5    0.05       0  5706.3    0.12       0
Bank Sta=5003.3,5009.3
Exp/Cntr=0.3,0.1

Type RM Length L Ch R = 1,3087,1793,1793,1793
BEGIN DESCRIPTION:
UNT166 IN CCTC 2.0
END DESCRIPTION:
XS GIS Cut Line= 3
      3566446.30     10669820.09      3567379.46     10666629.99
      3566185.92     10666315.33
#Sta/Elev= 30
  1426.3  324.14  1551.2  318.36  1559.6  316.31  1564.8  316.89  1598.2  312.84
  1658.6  309.34  1775.9  301.58  2020.0  291.49  2079.1  290.39  2279.5  288.82
  2521.3  288.30  3207.9  290.23  4395.6  289.26  4832.7  290.63  4927.0  292.75
  4977.4  292.55  4987.8  291.22  4995.1  286.20  4997.9  285.70  5001.1  286.20
  5009.0  290.13  5018.8  292.66  5215.3  292.37  5356.1  290.27  5517.3  291.28
  5673.3  300.55  5740.7  306.15  5904.8  316.49  5909.2  315.73  5984.4  318.54
#Mann=11,-1,0
  1426.3    0.16       0  1658.6    0.12       0  2020.0    0.16       0
  2079.1    0.05       0  2279.5     0.1       0  2521.3    0.05       0
  4927.0    0.12       0  4995.1    0.07       0  5001.1    0.12       0
  5740.7    0.16       0  5909.2    0.12       0
Bank Sta=4995.1,5001.1
Exp/Cntr=0.3,0.1

Type RM Length L Ch R = 1,1294,0,0,0
BEGIN DESCRIPTION:
UNT166 IN CCTC 1.0
END DESCRIPTION:
XS GIS Cut Line= 4
      3566793.52     10669646.48      3568095.60     10667378.69
      3568019.65     10666271.92      3565914.64     10665827.04
#Sta/Elev= 30
  2133.6  315.92  2414.4  297.12  2637.1  294.82  2956.5  290.29  3373.9  287.92
  3433.4  287.83  4303.9  288.95  4545.4  291.55  4656.8  290.50  4967.6  292.88
  4994.7  283.82  4997.5  283.32  5000.7  283.82  5017.7  292.96  5054.0  291.62
  5785.0  289.25  6144.2  291.84  6164.7  290.46  6174.9  291.88  6374.2  289.92
  7207.2  291.16  7401.4  296.46  7708.0  315.87  7789.8  316.46  7820.2  315.03
  7825.3  313.19  7833.6  313.98  7836.8  314.70  7869.9  317.60  8009.5  322.52
#Mann=9,-1,0
  2133.6    0.16       0  2637.1    0.05       0  3373.9    0.16       0
  3433.4    0.05       0  4656.8    0.12       0  4994.7    0.07       0
  5000.7    0.12       0  7833.6    0.16       0  7836.8    0.12       0
Bank Sta=4994.7,5000.7
Exp/Cntr=0.3,0.1

Chan Stop Cuts=-1
