--- ANDING BRANCH.prj (project) ---

Proj Title=ANDING BRANCH Base Level Engineering
Current Plan=p01
Default Exp/Contr=0.3,0.1
English Units
Geom File=g01
Flow File=f01
Plan File=p01
Y Axis Title=Elevation
X Axis Title(PF)=Main Channel Distance
X Axis Title(XS)=Station
BEGIN DESCRIPTION:
ANDING BRANCH
END DESCRIPTION:
DSS Export Rating Curves= 0
DSS Export Rating Curve Sorted= 0
DSS Export Volume Flow Curves= 0
DXF OffsetX= 0
DXF OffsetY= 0
DXF ScaleX= 1
DXF ScaleY= 10

--- ANDING BRANCH.p01 (plan) ---

Plan Title=Multiple Run
Short Identifier=Multiple
Geom File=g01
Flow File=f01
Subcritical Flow
K Sum by GR= 0
Std Step Tol= 0.01
Critical Tol= 0.01
Num of Std Step Trials= 20
Max Error Tol= 0.3
Flow Tol Ratio= 0.001
Split Flow NTrial= 30
Split Flow Tol= 0.02
Split Flow Ratio= 0.02
Log Output Level= 0
Friction Slope Method= 1
Unsteady Friction Slope Method= 2
Unsteady Bridges Friction Slope Method= 1
Parabolic Critical Depth
Global Vel Dist=  1 , 1 , 1
Global Log Level= 0
CheckData=True
Encroach Param= -1, 0, 0, 0
BEGIN DESCRIPTION:
Multiple Run
END DESCRIPTION:

--- ANDING BRANCH.f01 (steady flow) ---

Flow Title=Multiple
Program Version=4.10
Number of Profiles= 7
Profile Names=10-year,25-year,50-year,1pct_min,100-year,1pct_plu,500-year
River Rch & RM=ANDING BRANCH,Reach-1         ,28962
     752    1039    1279    1156    1563    2113    2338
River Rch & RM=ANDING BRANCH,Reach-1         ,28306
    1015    1419    1762    1602    2167    2930    3286
River Rch & RM=ANDING BRANCH,Reach-1         ,26682
    1272    1803    2259    2073    2804    3792    4330
River Rch & RM=ANDING BRANCH,Reach-1         ,25323
    1272    1803    2259    2073    2804    3792    4330
River Rch & RM=ANDING BRANCH,Reach-1         ,24208
    1379    1955    2448    2244    3034    4104    4676
River Rch & RM=ANDING BRANCH,Reach-1         ,18942
    1623    2318    2917    2685    3631    4911    5644
River Rch & RM=ANDING BRANCH,Reach-1         ,18494
    2231    3230    4103    3809    5151    6966    8143
River Rch & RM=ANDING BRANCH,Reach-1         ,18155
    2231    3230    4103    3809    5151    6966    8143
River Rch & RM=ANDING BRANCH,Reach-1         ,14595
    2320    3358    4264    3955    5349    7234    8447
River Rch & RM=ANDING BRANCH,Reach-1         ,11964
    2424    3505    4447    4121    5573    7537    8782
River Rch & RM=ANDING BRANCH,Reach-1         ,8853
    2587    3744    4755    4407    5960    8061    9399
River Rch & RM=ANDING BRANCH,Reach-1         ,7041
    2683    3884    4932    4571    6181    8360    9743
River Rch & RM=ANDING BRANCH,Reach-1         ,2854
    3370    4917    6278    5847    7908   10694   12586
River Rch & RM=ANDING BRANCH,Reach-1         ,695
    3370    4917    6278    5847    7908   10694   12586
Boundary for River Rch & Prof#=ANDING BRANCH,Reach-1         , 1
Up Type= 0
Dn Type= 3
Dn Slope=0.00294
Boundary for River Rch & Prof#=ANDING BRANCH,Reach-1         , 2
Up Type= 0
Dn Type= 3
Dn Slope=0.00294
Boundary for River Rch & Prof#=ANDING BRANCH,Reach-1         , 3
Up Type= 0
Dn Type= 3
Dn Slope=0.00294
Boundary for River Rch & Prof#=ANDING BRANCH,Reach-1         , 4
Up Type= 0
Dn Type= 3
Dn Slope=0.00294
Boundary for River Rch & Prof#=ANDING BRANCH,Reach-1         , 5
Up Type= 0
Dn Type= 3
Dn Slope=0.00294
Boundary for River Rch & Prof#=ANDING BRANCH,Reach-1         , 6
Up Type= 0
Dn Type= 3
Dn Slope=0.00294
Boundary for River Rch & Prof#=ANDING BRANCH,Reach-1         , 7
Up Type= 0
Dn Type= 3
Dn Slope=0.00294
DSS Import GetInterval= 0
DSS Import GetPeak= 0
DSS Import FillOption= 0

--- ANDING BRANCH.g01 (geometry) ---

Geom Title=Existing Conditions
Program Version=4.10

River Reach=ANDING BRANCH   ,Reach-1
Reach XY= 30
       3666271.5     10752834.75      3665931.75       10752572.
      3665787.25       10752048.       3665849.5       10750650.
       3665743.5       10749957.      3665938.75       10749238.
        3666278.       10748770.      3666530.25       10747960.
       3666926.5       10747714.        3667266.       10747673.
        3667420.       10747501.      3667397.25       10747344.
      3667749.25       10746985.      3667982.25       10746291.
        3668339.       10745810.      3668262.75       10745634.
      3668482.75       10744433.        3671576.       10742798.
       3671545.5       10742664.      3671993.75       10742055.
        3672646.       10741440.        3673579.       10741644.
        3674434.       10741424.      3675490.75       10740674.
      3676299.75       10740451.       3676885.5       10739955.
      3678653.75       10737767.        3679728.       10737936.
       3681398.5       10736215.      3682429.75       10733755.

Type RM Length L Ch R = 1 ,28962   ,656,656,656
BEGIN DESCRIPTION:
ANDING BRANCH 60.0
END DESCRIPTION:
XS GIS Cut Line= 3
      3666249.65     10752510.16      3665999.61     10752660.19
      3665799.58     10752910.23
#Sta/Elev= 30
    4709  420.79  4767.4  417.43    4781   415.8  4790.7  415.72  4802.3  414.22
  4839.3  411.65    4849  411.49  4860.7  409.39  4876.2  408.31    4884  406.56
  4891.8  405.76  4942.3     403    4987  402.04  4989.8  401.46  4992.6  400.96
  4995.8  401.46  4997.7  402.18  5007.8  401.74  5071.8  402.36  5100.6  403.35
  5164.7  407.41  5199.9  410.28  5214.3  412.04  5228.7  412.71  5235.1  413.75
  5243.1  413.89  5284.7  417.43  5313.5  418.25  5317.5  419.22  5320.8  419.22
#Mann= 3 ,-1 , 0
    4709     .05       0  4989.8     .03       0  4995.8     .05       0
Bank Sta=4987,4997.7
XS Rating Curve= 0 ,0
Exp/Cntr=0.3,0.1

Type RM Length L Ch R = 1 ,28306   ,79,79,79
BEGIN DESCRIPTION:
ANDING BRANCH 59.0
END DESCRIPTION:
XS GIS Cut Line= 2
      3666395.75     10752070.39       3665063.5     10752028.76
#Sta/Elev= 30
  4392.9  420.35  4449.1  417.78  4482.2  417.49  4581.2  413.77  4680.1  411.58
  4749.2   409.1  4799.2  408.48  4877.9  405.02  4939.3  402.91  4949.3  403.34
  4989.3   400.6  5039.4  400.76  5046.4  400.16  5049.1  399.66  5052.4  400.16
  5059.4  400.71  5075.8   401.2  5139.4  402.36  5159.4  406.03  5202.1  409.66
  5209.4  411.38  5239.5  414.93  5269.5  419.46  5319.5  423.86  5349.5  424.75
  5372.5   426.4  5439.5  427.34  5599.6  423.92  5679.7  425.01  5725.8  426.49
#Mann= 9 ,-1 , 0
  4392.9     .08       0  4482.2     .05       0  4581.2     .08       0
  4680.1     .05       0  4877.9     .08       0  5046.4     .07       0
  5052.4     .08       0  5075.8     .05       0  5372.5     .08       0
Bank Sta=5039.4,5059.4
XS Rating Curve= 0 ,0
Exp/Cntr=0.3,0.1

Type RM Length L Ch R = 1 ,28227   ,608,608,608
BEGIN DESCRIPTION:
ANDING BRANCH 58.0
END DESCRIPTION:
XS GIS Cut Line= 2
      3666434.89     10751992.27      3665036.41      10751950.6
#Sta/Elev= 30
  4350.2  420.72  4495.5  415.93  4584.2  411.61  4615.6  411.36  4677.1  408.86
  4905.7  402.47  4922.2  402.98  4927.2  401.88  4965.7  402.08  5012.8  400.38
  5015.5  399.88  5018.8  400.38  5035.8  402.68  5045.8  401.74  5061.9  401.98
  5135.8  403.24  5145.8  403.22  5185.8  406.44  5225.9  411.82  5260.1   414.6
  5265.9  416.05  5315.9  419.86  5365.9  425.52  5385.9  426.59    5436  426.48
    5506   424.3    5526  424.75  5561.8  422.95    5636  422.96  5749.3  426.53
#Mann= 6 ,-1 , 0
  4350.2     .05       0  4677.1     .12       0  5012.8     .07       0
  5018.8     .12       0  5061.9     .16       0  5561.8     .05       0
Bank Sta=4922.2,5135.8
XS Rating Curve= 0 ,0
Exp/Cntr=0.3,0.1

Type RM Length L Ch R = 1 ,27619   ,501,501,501
BEGIN DESCRIPTION:
Mapping XS 20cbf83c
END DESCRIPTION:
XS GIS Cut Line= 3
      3666649.65      10751610.2      3665849.61     10751410.19
      3665449.58     10751110.17
#Sta/Elev= 30
  4175.2  427.17  4257.7  423.35  4474.2  416.03  4528.3  413.43    4536   412.4
  4546.3  412.02  4556.6  410.64  4564.4  410.31  4569.5  410.75  4587.6  409.17
  4610.7  408.61  4618.5  407.48    4652  404.73  4700.9  403.43  4729.3  401.47
  4734.4  401.31  4742.2  399.64  4749.5  399.31  4752.2  398.81  4755.5  399.31
  5342.6  399.31  5363.4  401.42  5366.7   402.3  5375.9  404.47  5386.3  406.87
  5399.9  408.38  5413.4  410.98  5463.4  414.66    5478  414.28  5499.9  415.44
#Mann= 5 ,-1 , 0
  4175.2     .05       0  4749.5    .033       0  4755.5     .05       0
  5366.7     .16       0  5375.9     .12       0
Bank Sta=4729.3,5363.4
XS Rating Curve= 0 ,0
Exp/Cntr=0.3,0.1

Type RM Length L Ch R = 1 ,27118   ,436,436,436
BEGIN DESCRIPTION:
Mapping XS ff586ceb
END DESCRIPTION:
XS GIS Cut Line= 3
      3666644.64     10751311.75      3665835.64     10750902.04
      3665505.79     10751051.33
#Sta/Elev= 30
  4108.7  423.95  4114.3  423.17  4136.8  422.22  4143.9  421.51  4159.2  421.28
  4166.1  420.55  4305.4   416.4  4327.7  415.91  4338.5  416.07  4394.6   414.3
  4427.8  412.38  4439.4  411.03  4455.7  410.54  4461.8  409.65  4472.4  409.15
  4484.3  407.45  4494.7     407  4506.7  405.62  4583.8  401.38  4603.1  399.31
  4605.8  398.81  4609.1  399.31  5238.8  399.31  5261.9  401.48  5265.7  402.16
    5285  404.17  5307.6  407.79  5336.7  411.64  5365.3  413.87  5377.6  414.16
#Mann= 4 ,-1 , 0
  4108.7     .05       0  4603.1    .033       0  4609.1     .05       0
  5265.7     .16       0
Bank Sta=4583.8,5261.9
XS Rating Curve= 0 ,0
Exp/Cntr=0.3,0.1

Type RM Length L Ch R = 1 ,26682   ,469,469,469
BEGIN DESCRIPTION:
ANDING BRANCH 55.0
END DESCRIPTION:
XS GIS Cut Line= 3
      3666599.61     10750960.19      3665799.61     10750460.19
      3664599.62     10750060.19
#Sta/Elev= 30
  4083.8  417.09  4164.6  413.56  4301.4  410.68  4343.8  407.28  4359.2  407.91
  4374.5  405.63  4468.8  404.57  4474.7   405.7  4547.8  406.06  4584.4  404.83
  4620.9  401.26  4639.2  399.31  4641.9  398.81  4645.2  399.31  5562.1  399.31
  5659.7  399.31  5670.2  399.85  5680.7  402.84  5691.3  402.74  5710.2  405.11
  5807.2  411.15  5891.6  412.36  5933.7  415.89  5954.8  419.11  5965.3  416.57
  5986.4     419  6123.5  425.36  6218.3  432.53  6249.9  438.62  6292.1  443.93
#Mann= 5 ,-1 , 0
  4083.8     .05       0  4639.2    .033       0  4645.2     .05       0
  5562.1     .16       0  5710.2     .05       0
Bank Sta=4620.9,5680.7
XS Rating Curve= 0 ,0
Exp/Cntr=0.3,0.1

Type RM Length L Ch R = 1 ,26213   ,465,465,465
BEGIN DESCRIPTION:
ANDING BRANCH 54.0
END DESCRIPTION:
XS GIS Cut Line= 3
       3666949.6     10750810.18      3665749.61     10750010.19
      3665199.58     10749410.15
#Sta/Elev= 30
  3560.5  433.14  3596.5  430.83  3632.6  430.02  3776.8  419.93    3921  413.06
  4036.7  410.56  4072.8  411.46  4123.9  409.85    4196  409.79  4259.1   407.8
  4382.3  409.79  4448.4  408.19  4497.9  404.32  4547.5  403.32  4562.5  401.29
    4567  399.31  4569.8  398.81    4573  399.31  5257.7  399.31  5278.7  401.13
    5307  400.68  5314.4  399.31  5526.5  399.31  5540.7  401.12    5590  412.01
    5661  419.24  5717.7   422.2  5746.1  422.22  5788.6  424.73  5816.7  424.93
#Mann= 3 ,-1 , 0
  3560.5     .05       0    4567    .033       0    4573     .05       0
Bank Sta=4562.5,5540.7
XS Rating Curve= 0 ,0
Exp/Cntr=0.3,0.1

Type RM Length L Ch R = 1 ,25748   ,425,425,425
BEGIN DESCRIPTION:
ANDING BRANCH 53.0
END DESCRIPTION:
XS GIS Cut Line= 3
      3667049.61     10750660.19      3665849.61     10749560.19
      3665249.66      10749410.2
#Sta/Elev= 30
  3373.8  437.33  3515.3  428.93  3557.9  423.55    3643  418.68  3663.9  414.75
  3678.1  415.71  3734.8  413.27  3741.6  416.18    3749  414.74  3755.8  416.59
    3770  416.16  3777.4  414.08    3876  412.85  3911.8  409.74    4032  406.39
  4046.2   404.5  4081.4  403.96  4088.8  406.42  4117.1  407.73  4329.3  408.85
  4704.2   406.3  4782.5  401.17  4800.4  399.31  4803.2  398.81  4806.4  399.31
  5331.5  399.31  5341.8  401.22  5390.8  408.14  5465.5  414.96  5620.1     424
#Mann= 3 ,-1 , 0
  3373.8     .05       0  4800.4    .033       0  4806.4     .05       0
Bank Sta=4782.5,5341.8
XS Rating Curve= 0 ,0
Exp/Cntr=0.3,0.1

Type RM Length L Ch R = 1 ,25323   ,59,59,59
BEGIN DESCRIPTION:
Mapping XS 852b2ab3
END DESCRIPTION:
XS GIS Cut Line= 4
      3667083.59     10749685.56      3666346.34     10749364.97
      3665697.47     10749002.55      3665107.92     10748498.07
#Sta/Elev= 30
  3797.4  420.41    3920  414.38  4152.8  410.91  4176.2  409.02  4336.1  404.71
  4347.7  402.74  4390.6  400.98  4398.1   399.6  4470.9  396.76  4473.6  396.26
  4476.9  396.76  4543.3  401.56  4559.5  402.76  4623.8  403.28  4683.2   401.1
  4689.2  399.31  5294.4  399.31  5352.1  404.42  5380.7  402.11  5387.2  402.94
  5394.4  400.29  5408.1  399.76  5415.8  397.31  5450.9  399.34  5458.6   402.3
  5479.4   404.8  5550.8  402.99  5657.3  406.26    5834  403.93  6120.5  410.13
#Mann= 5 ,-1 , 0
  3797.4     .05       0  4347.7     .16       0  4470.9    .033       0
  4476.9     .16       0  4559.5     .05       0
Bank Sta=4390.6,4543.3
XS Rating Curve= 0 ,0
Exp/Cntr=0.3,0.1

Type RM Length L Ch R = 1 ,25264   ,61,61,61
BEGIN DESCRIPTION:
Mapping XS 1812457b
END DESCRIPTION:
XS GIS Cut Line= 4
      3667097.51     10749671.69      3666352.85      10749325.9
       3665803.8     10748978.68      3665104.54     10748466.89
#Sta/Elev= 30
  3804.9  422.45  3848.1  418.47  3956.9  413.74  4144.4  411.24  4353.9  404.92
    4420  400.23  4505.8   396.8  4563.4  400.53  4602.9  403.38  4677.1  400.73
    4762  402.66  4942.3  402.11  4980.8  400.38  4986.7  402.48  5013.9  402.35
  5038.4  400.88  5044.3  402.63  5241.9  401.73  5342.7  403.43  5413.9  401.42
  5434.8  397.43  5461.1  396.19  5463.8  395.69  5467.1  396.19  5470.3  399.78
  5499.6  403.48  5635.5  405.38  5727.4  402.43  5900.4  403.54  6142.1  410.42
#Mann= 5 ,-1 , 0
  3804.9     .05       0  4942.3     .16       0  5013.9     .05       0
  5461.1     .07       0  5467.1     .05       0
Bank Sta=4420,4563.4
XS Rating Curve= 0 ,0
Exp/Cntr=0.3,0.1

Type RM Length L Ch R = 1 ,25203   ,326,326,326
BEGIN DESCRIPTION:
ANDING BRANCH 52.0
END DESCRIPTION:
XS GIS Cut Line= 3
       3667104.5     10749647.41      3666348.51     10749256.46
      3665107.97     10748446.02
#Sta/Elev= 30
  3812.3  421.46  3947.5  414.36  4318.3  407.16  4489.8  396.74    4584   398.4
  4644.8  403.17  4703.1  402.42  4733.3  400.73  4781.5  391.68    4863  385.96
    4880  384.84  4920.3  384.32  4941.4  380.66  4956.5  383.37  5046.5  380.47
  5065.1  382.79  5068.1  379.26  5070.8  378.76  5074.1  379.26  5086.2  383.58
  5092.2   381.5  5151.8  385.39  5215.9  389.92    5231  394.21  5303.4  401.91
    5412  398.53  5426.6  394.71  5505.5   402.7  5728.7  400.89  6145.2  410.76
#Mann= 5 ,-1 , 0
  3812.3     .05       0    4880     .16       0  5046.5     .05       0
  5068.1     .07       0  5074.1     .05       0
Bank Sta=4863,5151.8
XS Rating Curve= 0 ,0
Exp/Cntr=0.3,0.1

Type RM Length L Ch R = 1 ,24877   ,335,335,335
BEGIN DESCRIPTION:
Mapping XS 70157ca1
END DESCRIPTION:
XS GIS Cut Line= 3
      3666399.65     10748810.19      3666249.61     10748810.19
      3666049.59     10748410.15
#Sta/Elev= 30
  4855.3  392.15  4865.3  391.19  4875.3  388.69  4885.3  388.01  4905.3  384.66
  4955.3  381.68  4965.3  380.24  4982.3  375.63  4985.1  375.13  4988.3  375.63
  4995.3  376.25  5002.8  380.04  5019.3   381.5  5080.8   381.8  5086.4  382.53
  5161.7   382.2    5215  383.68  5241.2  383.64  5265.3  386.42  5273.7  386.23
  5304.4  388.26  5326.8   391.5  5363.1  394.21  5371.5   394.2  5377.1  396.76
  5385.5  397.28  5399.4  400.01  5416.2   402.1  5438.6  403.63  5452.6  403.22
#Mann= 5 ,-1 , 0
  4855.3     .12       0  4982.3     .07       0  4988.3     .12       0
  5161.7     .07       0  5241.2     .05       0
Bank Sta=4955.3,5019.3
XS Rating Curve= 0 ,0
Exp/Cntr=0.3,0.1

Type RM Length L Ch R = 1 ,24542   ,223,223,223
BEGIN DESCRIPTION:
Mapping XS 2253d5e9
END DESCRIPTION:
XS GIS Cut Line= 2
      3666588.34     10748647.15      3666145.61     10748356.34
#Sta/Elev= 30
  4738.3   397.9  4796.7  396.12  4835.7     394  4844.5  392.66  4850.8   392.9
  4856.8   391.3  4871.9  389.97    4902  385.33  4912.2  385.15  4965.3  379.13
  4974.4  377.01  4980.4  377.34    4985   374.7  4987.8   374.2    4991   374.7
  4995.4  375.92  5001.4  375.89  5010.5  378.31  5016.5  377.39  5023.9   379.7
  5027.7  379.68  5095.7  380.72  5161.2  382.61  5167.5  384.25  5218.4  388.66
  5239.5  392.25  5248.6  394.44  5254.6  394.94  5262.6  397.44    5268  397.44
#Mann= 6 ,-1 , 0
  4738.3     .05       0  4796.7     .16       0  4912.2     .12       0
    4985     .07       0    4991     .12       0  5027.7     .05       0
Bank Sta=4965.3,5023.9
XS Rating Curve= 0 ,0
Exp/Cntr=0.3,0.1

Type RM Length L Ch R = 1 ,24319   ,111,111,111
BEGIN DESCRIPTION:
ANDING BRANCH 50.0
END DESCRIPTION:
XS GIS Cut Line= 6
      3666916.05     10748571.21      3666818.38      10748447.5
      3666646.94     10748349.85      3666269.34     10748271.72
       3666206.4     10748217.47      3666221.59       10747725.
#Sta/Elev= 30
  4393.5  398.29  4433.7     393  4470.7  394.08  4520.4  387.89  4526.8  391.08
  4534.8  387.52  4541.2  390.83  4561.4  387.77  4571.5  389.46  4634.9  383.18
  4651.7  381.75  4679.5  378.15  4687.8  381.29  4732.9  382.88  4738.6  376.57
    4744  381.34  4756.2  382.71  4922.9  379.71    4935  376.15  4982.3   374.4
  4985.1   373.9  4988.3   374.4  5065.8  379.58  5139.6  381.58  5158.9  385.51
  5179.8  383.09    5237  388.07  5417.2  393.36  5627.3  409.04  5712.5  409.88
#Mann= 5 ,-1 , 0
  4393.5     .05       0  4634.9     .16       0  4651.7     .05       0
  4982.3     .04       0  4988.3     .05       0
Bank Sta=4922.9,5065.8
XS Rating Curve= 0 ,0
Exp/Cntr=0.3,0.1

Type RM Length L Ch R = 1 ,24208   ,332,332,332
BEGIN DESCRIPTION:
ANDING BRANCH 49.0
END DESCRIPTION:
XS GIS Cut Line= 6
      3666974.62     10748536.46      3666777.15     10748291.25
      3666484.18      10748193.6      3666356.14     10748167.55
      3666299.72      10748091.6      3666288.87     10747748.71
#Sta/Elev= 30
  4291.6  397.67  4335.6  397.47  4356.4  394.23  4385.2  396.54  4420.4  394.18
  4434.8  395.71  4556.3  393.22  4562.8  391.54  4606.4  393.45  4654.3   389.6
  4659.5  391.58  4685.9   385.9  4740.9  382.61  4941.5  377.88  4970.9  376.48
  4981.1  374.46  4988.4  368.42  4991.1  367.92  4994.4  368.42  5001.6  368.83
  5007.1  375.38  5012.2  376.02  5063.3  378.78  5069.5  381.63  5092.5  381.15
  5119.6  385.48    5242  390.45    5330   398.4  5439.8   405.6  5483.6  406.75
#Mann= 6 ,-1 , 0
  4291.6     .05       0  4941.5     .16       0  4988.4     .07       0
  4994.4     .16       0    5330     .12       0  5439.8     .07       0
Bank Sta=4970.9,5012.2
XS Rating Curve= 0 ,0
Exp/Cntr=0.3,0.1

Type RM Length L Ch R = 1 ,23876   ,314,314,314
BEGIN DESCRIPTION:
Mapping XS 4eedf76b
END DESCRIPTION:
XS GIS Cut Line= 2
       3666896.5     10748273.88      3666370.02     10747654.24
#Sta/Elev= 30
  4516.4  396.39  4615.8  394.62  4715.8  384.01  4765.2  379.54  4836.2   376.7
  4919.2  377.75  4970.6  378.08  4978.3   374.4  4984.9  374.73  4992.6  371.17
  4999.1  366.54  5003.8  366.38  5006.5  365.88  5009.8  366.38  5013.4   377.2
    5020  378.32  5048.6  379.57  5084.8  379.86  5155.1  382.95  5170.3  384.25
  5240.8  388.86  5255.1  390.64  5261.6  392.24  5275.9  392.92  5282.5  394.07
  5290.2  393.95  5296.8  396.26  5304.5  396.33  5311.1  398.43  5329.5  400.45
#Mann= 5 ,-1 , 0
  4516.4     .05       0  4919.2     .12       0  5003.8     .07       0
  5009.8     .12       0  5170.3     .16       0
Bank Sta=4970.6,5020
XS Rating Curve= 0 ,0
Exp/Cntr=0.3,0.1

Type RM Length L Ch R = 1 ,23562   ,497,497,497
BEGIN DESCRIPTION:
ANDING BRANCH 48.0
END DESCRIPTION:
XS GIS Cut Line= 3
      3666999.61     10748060.19      3666849.61     10747760.19
      3666449.61     10747460.19
#Sta/Elev= 30
  4700.1  391.48  4753.2  385.77    4893  376.46  4946.1  375.05  4968.4  375.41
  4976.8  373.62  4990.8  365.02  4996.2     365  4998.9   364.5  5002.2     365
  5004.8  368.07  5013.1  368.42  5021.5  372.14  5032.7  374.77  5112.9  375.54
  5251.6   378.2  5285.2   380.4  5335.5  384.46  5371.9  389.27    5399  393.33
  5407.4  395.74  5413.6  395.67    5422  397.72  5435.5  398.92  5442.8  400.69
  5478.2  404.74  5485.5  406.72  5492.1  407.27  5513.6  409.73  5535.5  410.93
#Mann= 8 ,-1 , 0
  4700.1     .12       0  4996.2     .07       0  5002.2     .12       0
  5112.9     .05       0  5251.6     .12       0  5285.2     .07       0
  5371.9     .16       0  5492.1     .12       0
Bank Sta=4968.4,5032.7
XS Rating Curve= 0 ,0
Exp/Cntr=0.3,0.1

Type RM Length L Ch R = 1 ,23065   ,467,467,467
BEGIN DESCRIPTION:
ANDING BRANCH 47.0
END DESCRIPTION:
XS GIS Cut Line= 3
       3667399.6     10747810.17      3667299.61     10747660.19
      3667149.59     10747360.16
#Sta/Elev= 30
  4799.8  387.74  4802.8  387.74  4807.3  386.32  4828.3   385.1  4843.3  380.64
  4858.4  378.19  4907.9  374.85  4930.5  374.56  4972.5  371.67    4977  369.99
  4982.8  369.99  4988.4  366.83    4991  363.18  4993.8  362.68    4997  363.18
  5002.4  363.48  5010.8   370.7  5016.4  372.97  5069.5  370.99  5100.2  372.09
  5122.6  371.32  5150.6  372.07  5189.7  376.32    5212  380.88  5217.6  382.88
    5226  384.41  5248.4  386.09  5262.4  388.69  5284.7  390.99  5315.5  392.47
#Mann= 3 ,-1 , 0
  4799.8     .16       0    4991     .07       0    4997     .16       0
Bank Sta=4972.5,5016.4
XS Rating Curve= 0 ,0
Exp/Cntr=0.3,0.1

Type RM Length L Ch R = 1 ,22598   ,446,446,446
BEGIN DESCRIPTION:
ANDING BRANCH 46.0
END DESCRIPTION:
XS GIS Cut Line= 3
      3667749.59     10747410.18      3667499.61     10747310.19
      3667299.61     10747060.19
#Sta/Elev= 30
  4698.4  390.88  4730.7  388.99  4737.4  387.36  4755.4  385.73  4784.5  381.56
  4796.7  378.74  4806.1  378.16  4850.5  371.18  4892.2  369.55  4958.2  369.16
  4964.9  366.36  4970.8  366.36  4974.8  364.04  4989.3  363.34  4995.7  363.99
  5000.7  362.09  5003.4  361.59  5006.7  362.09  5018.1  367.76  5024.5  368.47
  5045.3  371.05  5102.9  374.89  5117.3  377.34  5131.7  377.23  5152.5  380.15
  5173.3  381.58  5201.6  385.83  5210.2  388.49  5237.4  393.29  5287.8  398.25
#Mann= 5 ,-1 , 0
  4698.4     .05       0  4755.4     .16       0  5000.7     .07       0
  5006.7     .16       0  5201.6     .05       0
Bank Sta=4958.2,5024.5
XS Rating Curve= 0 ,0
Exp/Cntr=0.3,0.1

Type RM Length L Ch R = 1 ,22152   ,413,413,413
BEGIN DESCRIPTION:
ANDING BRANCH 45.0
END DESCRIPTION:
XS GIS Cut Line= 3
      3667949.62     10747010.19      3667749.61     10746960.19
      3667349.59     10746910.19
#Sta/Elev= 30
  4802.4  388.54  4820.5  387.19  4861.7  376.94  4866.8   376.9  4884.9  373.38
  4949.3  369.14  4977.6  365.91  4990.5  365.99  4995.3  360.53    4998  360.03
  5001.3  360.53    5006  362.75  5011.1  362.75  5018.6  365.18    5069  366.71
  5119.4  366.09  5159.7  367.56  5179.9  372.09    5190  375.13    5200   375.9
  5207.6  377.46  5212.6  377.25  5220.2  378.93  5288.2  385.98  5293.3  385.63
  5300.8  387.32  5351.2  392.21  5368.9  395.33  5373.9  394.56  5411.7  398.37
#Mann= 3 ,-1 , 0
  4802.4     .05       0  4995.3     .03       0  5001.3     .05       0
Bank Sta=4990.5,5018.6
XS Rating Curve= 0 ,0
Exp/Cntr=0.3,0.1

Type RM Length L Ch R = 1 ,21739   ,463,463,463
BEGIN DESCRIPTION:
ANDING BRANCH 44.0
END DESCRIPTION:
XS GIS Cut Line= 3
      3668049.62     10746860.21      3667949.61     10746610.19
      3667549.58     10746210.16
#Sta/Elev= 30
    4717   385.4  4731.8  384.93  4749.3  383.27  4756.3  381.33  4761.4  383.07
  4770.9  379.74  4785.7  378.68  4846.3  370.53    4888  368.75    4923  365.72
  4964.7  364.41  4971.5  361.56  4976.9  361.18  4980.6  359.88  4983.3  359.38
  4986.6  359.88  5014.6  363.85  5141.8   363.3  5240.8  364.15    5288  365.44
  5311.5  366.65  5325.7  366.58  5382.3  370.64  5438.8  377.95  5467.1  382.76
  5481.3  384.14  5509.5  390.69  5523.7  391.78  5548.4  398.03    5552  398.03
#Mann= 5 ,-1 , 0
    4717     .16       0  4756.3     .05       0  4980.6     .03       0
  4986.6     .05       0    5288     .16       0
Bank Sta=4964.7,5014.6
XS Rating Curve= 0 ,0
Exp/Cntr=0.3,0.1

Type RM Length L Ch R = 1 ,21276   ,454,454,454
BEGIN DESCRIPTION:
ANDING BRANCH 43.0
END DESCRIPTION:
XS GIS Cut Line= 3
      3668449.64     10746210.19      3668049.61     10746160.19
      3667749.57     10746010.17
#Sta/Elev= 30
  4602.6  374.57  4622.8  370.72  4663.1  368.76  4673.2  366.39    4721  363.34
  4814.3  361.44  4925.1     361  4975.5  361.97  4992.7   356.7  4995.4   356.2
  4998.7   356.7  5003.2  361.07  5019.7  360.55  5037.5  362.35  5064.4  361.58
  5095.2  362.52  5109.2  364.11  5117.5  366.65  5125.9  367.05  5131.5  368.95
  5146.1  370.22    5207  376.77  5215.4   379.3  5229.3  380.29  5237.7  382.44
  5260.1  386.06  5265.7  386.11  5274.1  387.89  5299.2  390.55  5341.2  394.35
#Mann= 6 ,-1 , 0
  4602.6     .12       0  4992.7     .07       0  4998.7     .12       0
  5037.5     .16       0  5146.1     .05       0  5299.2     .16       0
Bank Sta=4975.5,5003.2
XS Rating Curve= 0 ,0
Exp/Cntr=0.3,0.1

Type RM Length L Ch R = 1 ,20822   ,499,499,499
BEGIN DESCRIPTION:
ANDING BRANCH 42.0
END DESCRIPTION:
XS GIS Cut Line= 3
       3668599.6     10745910.18      3668299.61     10745810.19
      3667899.62     10745660.19
#Sta/Elev= 30
  4671.6  388.89  4682.1  388.61  4692.7  386.23  4703.2  386.28  4766.5  377.19
  4798.1  373.88  4819.2   370.3  4924.6  360.26  4935.1  357.08  4953.2  356.17
  4955.9  355.67  4959.2  356.17  4977.3  357.62  4997.6  357.08  5009.2  359.18
  5041.2     360  5088.4  358.57  5094.6  359.22  5143.6  358.68  5173.8  359.57
  5234.3  364.58  5288.5  370.19  5297.5  372.32  5308.2  372.66  5314.4  373.84
  5350.9  375.21  5393.7  380.03  5405.2   380.5  5412.3  382.84    5415  382.84
#Mann= 4 ,-1 , 0
  4671.6     .12       0  4953.2     .07       0  4959.2     .12       0
  5288.5     .05       0
Bank Sta=4924.6,5009.2
XS Rating Curve= 0 ,0
Exp/Cntr=0.3,0.1

Type RM Length L Ch R = 1 ,20323   ,473,473,473
BEGIN DESCRIPTION:
Mapping XS 9d0d9dad
END DESCRIPTION:
XS GIS Cut Line= 3
      3668499.63      10745460.2      3668349.61     10745410.19
      3667949.56     10745460.19
#Sta/Elev= 30
  4817.6  378.45  4828.2  377.85  4849.2  374.43  4859.8  370.53  4870.3  369.64
  4880.9  366.98  4891.4  366.26  4933.6  359.67  4965.2  357.12  4973.1  357.92
  4985.8  357.73  4995.9  356.24    5003   356.2  5005.7   355.7    5009   356.2
  5013.5  358.08  5066.4  357.96  5094.2  356.59  5167.2  357.22  5179.8  357.72
  5227.7  362.08  5260.4   365.6    5268   367.8  5273.8  368.27  5288.2  370.63
  5318.4  371.52  5341.1  373.15  5358.7  375.31  5368.8  377.34  5378.9  378.19
#Mann= 4 ,-1 , 0
  4817.6     .12       0    5003     .07       0    5009     .12       0
  5273.8     .05       0
Bank Sta=4985.8,5013.5
XS Rating Curve= 0 ,0
Exp/Cntr=0.3,0.1

Type RM Length L Ch R = 1 ,19850   ,441,441,441
BEGIN DESCRIPTION:
ANDING BRANCH 40.0
END DESCRIPTION:
XS GIS Cut Line= 3
      3668649.57     10745110.17      3668399.61     10744960.19
      3667999.62      10744760.2
#Sta/Elev= 30
  4679.6  381.18  4687.3  379.84  4702.9  379.23  4710.6  376.21  4745.6  367.02
  4761.2  365.39  4803.9  357.95  4825.9  356.25  4854.5  354.76  4862.3  355.71
  4957.5   356.6  5015.8  354.83  5124.6  353.99  5127.4  353.49  5130.6  353.99
  5158.4  354.01  5163.9  354.89  5172.3  354.97  5208.7  359.99  5217.1  359.77
  5231.7  362.09  5239.4  364.01  5284.2  369.98  5292.5  369.76  5314.9  373.73
  5320.5   376.1  5359.6  382.07    5382  384.24  5412.4  384.91  5418.3  385.36
#Mann= 8 ,-1 , 0
  4679.6     .16       0  4710.6     .12       0  4825.9     .16       0
  5124.6     .07       0  5130.6     .16       0  5163.9     .12       0
  5231.7     .05       0  5412.4     .16       0
Bank Sta=4761.2,5239.4
XS Rating Curve= 0 ,0
Exp/Cntr=0.3,0.1

Type RM Length L Ch R = 1 ,19409   ,467,467,467
BEGIN DESCRIPTION:
Mapping XS 73e62138
END DESCRIPTION:
XS GIS Cut Line= 3
      3668799.63     10744810.21      3668449.61     10744510.19
      3668149.63     10744660.18
#Sta/Elev= 30
  4548.4  375.19  4562.2   374.6  4590.7  370.97  4598.4  368.25  4612.6  365.31
    4629  361.88    4662  355.93  4697.2  354.03  4711.4  355.29    4740  353.85
  4811.3  354.69  4903.5  353.81  4910.1  355.09  4924.3  354.62  4927.9  353.26
  4930.7  352.76  4933.9  353.26  4955.7  353.26  5078.6  353.78  5107.2  353.96
  5143.6  356.08  5157.5  359.15  5202.1  363.21  5210.7  363.88  5224.6  366.01
  5241.4  366.52  5300.1  371.57  5308.5  371.42  5312.6  372.48  5344.8  374.34
#Mann= 8 ,-1 , 0
  4548.4     .12       0    4629     .16       0  4927.9    .033       0
  4933.9     .16       0  4955.7     .05       0  5078.6     .12       0
  5202.1     .16       0  5312.6     .05       0
Bank Sta=4612.6,5210.7
XS Rating Curve= 0 ,0
Exp/Cntr=0.3,0.1

Type RM Length L Ch R = 1 ,18942   ,448,448,448
BEGIN DESCRIPTION:
Mapping XS 17ef570e
END DESCRIPTION:
XS GIS Cut Line= 3
      3668799.61     10744760.19      3668799.61     10744210.19
      3668499.58     10743910.16
#Sta/Elev= 30
  4478.7  369.99  4481.2  369.99  4488.7  368.57  4498.7  365.96  4508.7  365.19
  4518.7  362.73  4528.7  361.68  4538.7  358.98  4548.7  358.13  4558.7  356.42
  4568.7  355.45  4578.7  353.98  4583.7  353.47  4585.7  353.26  4588.4  352.76
  4588.9  352.76  4591.7  353.26  5311.5  353.26  5325.7     354  5327.6  354.28
  5339.8  356.07    5354  358.84  5368.1   362.3  5382.3  365.52  5396.4  370.32
  5410.5  373.89  5424.7  376.94  5438.8  379.03  5449.4  380.05    5453  380.05
#Mann= 5 ,-1 , 0
  4478.7     .12       0  4583.7     .05       0  4585.7    .033       0
  4591.7     .05       0  5327.6     .16       0
Bank Sta=4508.7,5382.3
XS Rating Curve= 0 ,0
Exp/Cntr=0.3,0.1

Type RM Length L Ch R = 1 ,18494   ,339,339,339
BEGIN DESCRIPTION:
ANDING BRANCH 37.0
END DESCRIPTION:
XS GIS Cut Line= 3
       3669899.6     10744710.18      3669199.61     10744060.19
      3668449.59     10743610.18
#Sta/Elev= 30
  4068.7  368.73  4146.6   366.7  4189.1  363.75  4252.9  359.86  4273.6  359.16
  4287.8  356.95  4316.2  355.18  4327.3  353.26  4330.1  352.76  4333.3  353.26
  4383.3  353.26  5578.7  353.26  5630.4  354.22  5688.7  359.89    5710  364.43
    5720  364.99  5723.6  365.36  5731.4  368.51    5747  369.83    5782   375.1
  5789.7  377.74  5791.8  377.63  5795.6  377.44  5816.9  380.97  5832.5  381.63
    5848  385.89  5853.9  385.46  5875.3  387.96  5890.8  388.64  5898.6  390.29
#Mann= 8 ,-1 , 0
  4068.7     .12       0  4252.9     .16       0  4327.3    .033       0
  4333.3     .16       0  4383.3     .05       0  5578.7     .16       0
    5720     .12       0  5791.8     .16       0
Bank Sta=4189.1,5710
XS Rating Curve= 0 ,0
Exp/Cntr=0.3,0.1

Type RM Length L Ch R = 1 ,18155   ,914,914,914
BEGIN DESCRIPTION:
Mapping XS d7eda9ae
END DESCRIPTION:
XS GIS Cut Line= 2
      3670425.57     10744689.19      3668295.35     10742881.89
#Sta/Elev= 30
  3808.7  382.71  3882.7  383.03  3925.5  380.49  4067.2  363.72  4144.2  357.69
  4200.9  354.72  4227.9  353.26  4230.7  352.76  4233.9  353.26    4276  353.26
    5667  353.26  5713.8  353.26  5756.7  360.32  5770.5  364.47  5784.1  367.34
  5798.4  370.72  5825.8  372.57  5909.8  369.42  5933.5  368.77    5941  365.68
  5947.8  365.34  5976.4  371.56  6025.8  374.64  6040.1  377.84  6175.2  390.97
  6269.6     394  6437.7   397.8  6490.8     401  6538.1   403.9  6602.3  406.52
#Mann= 13 ,-1 , 0
  3808.7     .12       0  4144.2     .16       0  4200.9     .12       0
  4227.9    .033       0  4233.9     .12       0    4276     .05       0
    5667     .16       0  5784.1     .12       0  5825.8     .16       0
  5909.8     .12       0  6269.6     .16       0  6490.8     .05       0
  6538.1     .12       0
Bank Sta=4067.2,5770.5
XS Rating Curve= 0 ,0
Exp/Cntr=0.3,0.1

Type RM Length L Ch R = 1 ,17241   ,438,438,438
BEGIN DESCRIPTION:
ANDING BRANCH 34.0
END DESCRIPTION:
XS GIS Cut Line= 3
      3670849.58     10744010.16      3670299.61     10743460.19
      3668493.91     10742330.21
#Sta/Elev= 30
  4248.3  388.39  4275.3  386.59  4545.2  364.02  4601.8  358.56    4613  353.26
  4615.7  352.76    4619  353.26  4624.4  353.26  6013.4  353.26    6048  356.23
  6071.2  355.46  6165.5  364.07  6202.1  365.68  6253.3  375.41  6369.5  383.72
  6427.2  378.46  6490.9  376.76  6536.1  378.46  6600.5   376.1  6637.1  378.14
    6643   375.9  6652.4  378.91  6694.5  378.66  6731.4  381.54  6752.6  379.86
  6804.5   382.1  6951.5  382.19  7038.6  384.69  7093.3  386.58  7156.2  394.06
#Mann= 10 ,-1 , 0
  4248.3     .16       0  4275.3     .12       0    4613    .033       0
    4619     .12       0  4624.4     .05       0    6048     .12       0
  6253.3     .16       0  6694.5     .12       0  6951.5     .16       0
  7038.6      .1       0
Bank Sta=4545.2,6165.5
XS Rating Curve= 0 ,0
Exp/Cntr=0.3,0.1

Type RM Length L Ch R = 1 ,16803   ,347,347,347
BEGIN DESCRIPTION:
ANDING BRANCH 33.0
END DESCRIPTION:
XS GIS Cut Line= 3
       3670899.6     10743860.15      3670699.61     10743260.19
      3670040.58     10741273.88
#Sta/Elev= 30
  4375.5  377.96  4544.1  364.42  4564.5  362.48  4660.1  355.46  4667.6  353.26
  4670.4  352.76  4673.6  353.26  4697.4  353.26  5951.3  353.26  6011.2  353.26
  6042.8  358.85  6055.9  359.17  6093.1  362.06  6106.2  365.41  6112.9  366.05
    6176  376.04  6219.6  379.88  6227.7     384    6291  392.94  6322.7  393.53
    6328  392.03  6354.4  394.25  6359.7  392.38  6549.8  404.25  6644.8     403
  6771.5  392.42  6834.9  390.43    6893  391.08  7002.5  384.13  7100.7  380.31
#Mann= 10 ,-1 , 0
  4375.5     .12       0  4564.5     .16       0  4667.6    .033       0
  4673.6     .16       0  4697.4     .05       0  5951.3     .16       0
  6055.9     .12       0  6112.9     .16       0    6176     .12       0
  7002.5     .16       0
Bank Sta=4544.1,6106.2
XS Rating Curve= 0 ,0
Exp/Cntr=0.3,0.1

Type RM Length L Ch R = 1 ,16456   ,35,35,35
BEGIN DESCRIPTION:
Mapping XS c4b8192c
END DESCRIPTION:
XS GIS Cut Line= 6
      3671131.46     10743712.54      3671116.27     10743449.99
      3670944.83     10742885.76      3670953.51     10742683.94
      3671029.47     10742527.69      3670929.65     10742065.47
#Sta/Elev= 30
  4391.6   380.4    4434  379.03  4464.1  371.38  4484.1  363.74  4685.7  357.06
  4692.8  356.67  4695.1  353.26  4697.8  352.76  4701.1  353.26  4839.9  353.26
  4943.6  353.26  5135.1  353.26  5141.1  355.89  5150.9  353.26    5174  357.92
  5179.2  355.75  5206.9  361.55  5212.1  360.47  5239.4  368.15    5380  375.23
  5537.1  367.56    5620  370.18  5699.3  362.75  5770.9  359.42    5835  358.19
  5876.9  360.08  5960.7  362.36  5990.6  363.34  6057.4  367.88  6092.9  367.74
#Mann= 9 ,-1 , 0
  4391.6     .05       0  4695.1     .03       0  4701.1     .05       0
  4839.9     .16       0  4943.6     .05       0  5150.9     .16       0
  5876.9     .12       0  5960.7     .16       0  5990.6     .12       0
Bank Sta=4685.7,5174
XS Rating Curve= 0 ,0
Exp/Cntr=0.3,0.1

Type RM Length L Ch R = 1 ,16421   ,97,97,97
BEGIN DESCRIPTION:
Mapping XS b4bd9f5e
END DESCRIPTION:
XS GIS Cut Line= 4
      3671163.48     10743705.87      3671150.46     10743448.02
      3670996.81      10742932.4      3670970.77     10742737.13
#Sta/Elev= 30
  4383.8  378.29  4419.5     376  4439.6  372.47  4459.6  364.74  4489.6  362.64
  4658.9  362.92  4823.5  361.68  4835.1  362.57  4840.4  359.88  4868.3  362.56
  4870.5  358.65  4873.3  358.15  4876.5  358.65  4906.7  363.21  4911.9  359.46
    4927  361.38    4973  362.84  4978.2  360.36  5036.2  363.93  5049.8  361.55
  5077.7  364.15  5082.9  360.18  5109.3  364.17  5133.9  363.78  5161.4  363.67
  5262.9   364.3  5275.2  368.12  5303.3   369.7  5343.3  377.11    5377  377.21
#Mann= 6 ,-1 , 0
  4383.8     .05       0  4823.5     .16       0  4870.5     .03       0
  4876.5     .16       0    4927     .05       0  5133.9     .16       0
Bank Sta=4658.9,5161.4
XS Rating Curve= 0 ,0
Exp/Cntr=0.3,0.1

Type RM Length L Ch R = 1 ,16324   ,373,373,373
BEGIN DESCRIPTION:
Mapping XS 6b5bc0ad
END DESCRIPTION:
XS GIS Cut Line= 4
      3671244.38     10743724.45      3671236.57     10743385.87
      3671093.34     10742930.14      3671044.24     10742738.92
#Sta/Elev= 30
  4325.4  366.97  4390.7   366.3  4649.8  354.83  4700.1  348.11  4767.5  344.94
  4816.8  341.58  4942.6  337.58  4969.8  335.15    4975   337.3  4989.5  333.76
    4992  332.93  4994.7  332.43    4998  332.93  5002.2  333.03  5007.4  335.89
  5015.9   336.8  5039.8  339.06  5057.9   338.8  5075.6  340.34  5139.7   346.1
    5213  348.11  5218.1   351.2  5234.6  356.79  5253.7  360.74  5258.9  364.03
  5278.8  366.11  5294.5  366.26  5306.9  368.53  5335.2   370.2  5339.2   372.4
#Mann= 8 ,-1 , 0
  4325.4     .16       0  4390.7     .05       0  4767.5     .16       0
  4989.5     .12       0    4992     .07       0    4998     .12       0
  5075.6     .05       0  5278.8     .16       0
Bank Sta=4975,5015.9
XS Rating Curve= 0 ,0
Exp/Cntr=0.3,0.1

Type RM Length L Ch R = 1 ,15951   ,455,455,455
BEGIN DESCRIPTION:
ANDING BRANCH 31.0
END DESCRIPTION:
XS GIS Cut Line= 3
       3671649.6     10743460.16      3671449.61     10742860.19
      3670999.58     10742710.18
#Sta/Elev= 30
  4377.7  356.94  4388.2  355.45  4440.9  354.04  4451.5  352.63  4535.8   348.1
  4704.4  340.49  4894.2  335.72  4925.8  336.62  4957.4   335.1    4970  336.42
    4989  335.89  4996.6  333.95  4999.3  333.45  5002.6  333.95  5020.7  335.29
  5147.2  336.82  5199.9  339.97    5242  343.77  5251.8  345.58  5263.1  346.22
  5284.2     350  5336.9  356.78  5347.4  360.92  5379.1  367.02  5410.7  367.38
  5442.3  372.28  5452.8  372.32  5463.4   375.5  5473.9  377.28  5484.5  377.11
#Mann= 5 ,-1 , 0
  4377.7     .16       0    4970     .12       0  4996.6     .07       0
  5002.6     .12       0  5251.8     .16       0
Bank Sta=4989,5020.7
XS Rating Curve= 0 ,0
Exp/Cntr=0.3,0.1

Type RM Length L Ch R = 1 ,15496   ,489,489,489
BEGIN DESCRIPTION:
ANDING BRANCH 30.0
END DESCRIPTION:
XS GIS Cut Line= 3
      3672249.65     10742960.21      3671649.61     10742560.19
      3671149.56     10742560.19
#Sta/Elev= 30
  4254.7  364.06  4349.4  355.85  4355.4  354.36  4421.5  348.12  4427.5  348.48
  4457.6  345.89  4463.6   344.7  4493.6  344.35  4543.6  340.89  4571.7  338.56
  4658.9  335.52    4746  336.69  4795.6  333.99  4818.1  335.05  4911.3  333.07
  4968.3  333.96  4969.8  332.69  4972.6  332.19  4975.8  332.69  5015.9  333.69
  5099.5   334.3  5145.9  334.42  5198.5  336.43  5245.9  340.41  5297.5  343.37
  5365.9  352.42  5375.9  354.97  5405.9  358.58  5415.9  360.74  5475.9  366.42
#Mann= 7 ,-1 , 0
  4254.7     .16       0  4543.6     .12       0  4969.8     .07       0
  4975.8     .12       0  5099.5     .16       0  5198.5     .12       0
  5297.5     .16       0
Bank Sta=4968.3,5015.9
XS Rating Curve= 0 ,0
Exp/Cntr=0.3,0.1

Type RM Length L Ch R = 1 ,15007   ,412,412,412
BEGIN DESCRIPTION:
ANDING BRANCH 29.0
END DESCRIPTION:
XS GIS Cut Line= 3
      3672549.58     10742810.16      3671949.61     10742210.19
       3671449.6     10741710.18
#Sta/Elev= 30
  4154.1  381.17  4295.5  360.08  4366.2  353.49  4422.8  349.73  4436.9  347.07
  4521.8  340.88    4550  340.64  4620.7  335.59  4713.4  332.15  4790.5  332.75
  4830.9  331.61  4875.3  330.67  4931.9  333.36  4960.2  332.86  4974.3  330.85
  4988.4  330.56  5073.3  331.36  5087.4  329.87  5101.6   331.2  5129.9  331.05
    5141  329.35  5143.8  328.85    5147  329.35  5158.1  331.04  5407.8  331.59
  5469.3  335.23  5567.9  344.67  5610.7  348.95  5667.3  360.74  5709.7  366.51
#Mann= 7 ,-1 , 0
  4154.1     .16       0  4713.4     .12       0  4830.9     .05       0
    5141     .03       0    5147     .05       0  5407.8     .16       0
  5567.9     .12       0
Bank Sta=5129.9,5158.1
XS Rating Curve= 0 ,0
Exp/Cntr=0.3,0.1

Type RM Length L Ch R = 1 ,14595   ,664,664,664
BEGIN DESCRIPTION:
ANDING BRANCH 28.0
END DESCRIPTION:
XS GIS Cut Line= 3
      3672599.59     10742460.16      3672149.61     10741860.19
      3671274.78     10741019.58
#Sta/Elev= 30
  4274.2  355.56  4310.6  351.03  4424.2  341.25  4516.9  333.95  4557.7  332.78
  4602.3  330.49  4737.4  330.39  4752.3  329.21  4802.3   330.9  4882.7  330.51
    4996  328.81  4999.3  327.49    5002  326.99  5005.3  327.49  5024.2  328.77
  5215.2   329.2  5264.6  330.97  5448.5  329.21    5557  332.92  5724.3  343.99
  5780.9  351.09  5865.8  358.06  5886.9  358.54  5894.1  360.32  5929.4  360.87
  6035.6  369.21  6113.3  371.42  6176.9  370.33  6226.5  372.54  6237.4   371.8
#Mann= 7 ,-1 , 0
  4274.2     .16       0  4557.7     .05       0  4737.4      .1       0
  4882.7     .05       0  4999.3    .033       0  5005.3     .05       0
    5557     .16       0
Bank Sta=4996,5024.2
XS Rating Curve= 0 ,0
Exp/Cntr=0.3,0.1

Type RM Length L Ch R = 1 ,13931   ,49,49,49
BEGIN DESCRIPTION:
ANDING BRANCH 27.0
END DESCRIPTION:
XS GIS Cut Line= 5
      3672804.21     10742499.38      3672806.08     10742132.94
      3672582.77     10741159.93      3672484.85     10741071.19
      3672432.65     10740703.27
#Sta/Elev= 30
  3922.6  371.57  3971.8  367.17  4003.5  365.98  4091.8  359.56  4221.8  345.95
  4287.9  341.05  4332.9   339.2  4344.3  337.46  4430.1  333.98  4507.3  334.76
  4578.6  332.51  4649.5  329.15    4689  327.49  4691.8  326.99    4695  327.49
  5199.2  327.49  5221.5  327.49  5367.4   328.1  5409.9  331.51  5416.2  333.24
  5423.4  332.73  5430.6  334.07    5471   336.2  5489.3   339.1  5494.3   341.4
  5511.4  343.14  5521.5  347.37  5551.8   349.1  5616.4  354.99  5791.1  370.62
#Mann= 8 ,-1 , 0
  3922.6     .16       0  4578.6     .05       0    4689    .033       0
    4695     .05       0  5199.2     .12       0  5221.5     .05       0
  5416.2     .16       0  5616.4     .12       0
Bank Sta=4649.5,5367.4
XS Rating Curve= 0 ,0
Exp/Cntr=0.3,0.1

Type RM Length L Ch R = 1 ,13882   ,40,40,40
BEGIN DESCRIPTION:
Mapping XS 257b87e3
END DESCRIPTION:
XS GIS Cut Line= 6
      3672861.95     10742117.66      3672629.32     10741169.79
      3672573.77     10741065.62      3672507.79     10741065.62
       3672493.9     10741006.59      3672473.07     10740687.13
#Sta/Elev= 30
  4302.3  342.99  4351.1   338.7  4433.4  336.51  4590.4  335.61  4626.8  337.52
  4631.9   334.8  4659.9   337.5  4668.3   337.4  4673.4  334.21  4701.1  337.22
  4721.7   334.9  4751.2  337.75  4756.4  335.62  4778.8  336.53    4965  337.32
    5067  337.24  5129.7  335.19    5247  336.83  5254.2   334.4  5259.3  336.73
  5351.8  336.75  5357.5  333.15  5377.2  333.34    5425   335.5  5459.6  332.21
  5462.4  331.71  5465.6  332.21  5522.9  337.18  5563.9  345.39  5844.6   370.9
#Mann= 9 ,-1 , 0
  4302.3     .16       0  4756.4     .12       0  4778.8     .05       0
    4965     .16       0    5067     .12       0  5377.2     .16       0
  5459.6     .07       0  5465.6     .16       0  5563.9     .12       0
Bank Sta=5351.8,5522.9
XS Rating Curve= 0 ,0
Exp/Cntr=0.3,0.1

Type RM Length L Ch R = 1 ,13842   ,531,531,531
BEGIN DESCRIPTION:
ANDING BRANCH 26.0
END DESCRIPTION:
XS GIS Cut Line= 3
      3672988.91     10742173.45      3672874.36     10742024.18
       3672561.9     10740704.94
#Sta/Elev= 30
  4211.5  360.66  4277.8  353.18  4398.8  337.64  4620.1  333.74  4650.4  330.93
  4718.6  327.93  4878.7  329.06  4907.3  327.19  4920.8  328.86  4963.5  328.47
  5005.5  327.45  5010.6  330.53  5030.6  327.68  5065.2  327.65  5140.7  326.61
  5143.4  326.11  5146.7  326.61  5316.6  328.08  5390.3  327.44  5438.2  331.59
  5485.6  335.22  5503.4  339.92  5557.5  345.96  5654.6   361.8  5659.8  360.58
  5696.9  368.42    5702  367.25  5739.1  374.01  5744.3  372.56  5755.4  376.31
#Mann= 10 ,-1 , 0
  4211.5     .12       0  4277.8     .16       0  4718.6     .12       0
  4920.8     .05       0  4963.5     .16       0  5065.2     .12       0
  5140.7     .07       0  5146.7     .12       0  5316.6     .16       0
  5557.5     .12       0
Bank Sta=4650.4,5438.2
XS Rating Curve= 0 ,0
Exp/Cntr=0.3,0.1

Type RM Length L Ch R = 1 ,13311   ,333,333,333
BEGIN DESCRIPTION:
ANDING BRANCH 25.0
END DESCRIPTION:
XS GIS Cut Line= 3
      3672999.61     10742110.17      3673199.61     10741510.19
       3672699.6     10740510.17
#Sta/Elev= 30
  4384.7  355.07  4385.2  355.07    4469  340.26  4553.3  331.59    4582  327.76
  4627.1  325.49  4837.9  324.42    4975  325.26  4985.5  327.51  5011.5  324.11
  5014.3  323.61  5017.5  324.11  5036.5  324.11  5047.9  324.11  5061.9  327.89
  5119.1   325.8  5260.1  325.07  5324.5  325.07  5478.3  325.07  5495.1  328.81
  5545.4  326.82  5612.5  330.63  5707.1  341.82  5735.3  344.82  5808.7  353.28
  5875.2  361.28  5970.3  380.39  6054.1  393.45  6104.4  399.61  6135.2  399.42
#Mann= 12 ,-1 , 0
  4384.7     .12       0  4385.2     .16       0    4582     .12       0
  5011.5     .07       0  5017.5     .12       0  5036.5     .07       0
  5119.1     .12       0  5260.1     .05       0  5324.5     .16       0
  5707.1     .12       0  5735.3     .16       0  5808.7     .12       0
Bank Sta=4553.3,5612.5
XS Rating Curve= 0 ,0
Exp/Cntr=0.3,0.1

Type RM Length L Ch R = 1 ,12978   ,472,472,472
BEGIN DESCRIPTION:
Mapping XS ca88d821
END DESCRIPTION:
XS GIS Cut Line= 3
      3673205.77     10742684.99      3673445.36     10741888.08
      3673575.57     10740596.37
#Sta/Elev= 30
  3917.7  362.87  3992.3  353.66  4048.5  348.24  4115.3  341.06  4228.5  330.62
  4371.7  324.95  4505.4  324.11  4508.2  323.61  4511.4  324.11  4641.7  325.93
  4645.7  324.11  4699.6   325.6  4742.9  325.64  4841.3  324.11  4939.4  324.11
  5037.5  324.11  5119.6  324.11    5143  326.73  5233.8  324.11  5290.5  326.31
  5331.9  324.11    5391  324.11  5411.1  328.52  5438.2  325.67  5528.2  325.95
  5593.8  326.05  5632.2  327.01  5662.3  331.17  5903.6  370.71  6048.1  379.82
#Mann= 16 ,-1 , 0
  3917.7     .12       0  3992.3     .16       0  4048.5     .12       0
  4115.3     .16       0  4505.4     .07       0  4511.4     .16       0
  4641.7     .12       0  4699.6     .05       0  4742.9     .16       0
  4841.3     .12       0  4939.4     .07       0  5037.5     .16       0
  5233.8      .1       0  5331.9     .07       0  5528.2     .16       0
  5593.8     .12       0
Bank Sta=4228.5,5662.3
XS Rating Curve= 0 ,0
Exp/Cntr=0.3,0.1

Type RM Length L Ch R = 1 ,12506   ,281,281,281
BEGIN DESCRIPTION:
Mapping XS c9871432
END DESCRIPTION:
XS GIS Cut Line= 4
      3673898.49     10742893.27      3673987.03     10741924.53
      3673825.57     10740856.83      3673815.16     10740554.92
#Sta/Elev= 30
  3657.1  378.71  3719.9  378.56  3730.5  380.02  3954.3  368.79  4182.4  348.82
  4253.4  346.26    4343  343.88    4491  333.81  4496.1  335.15  4594.1  330.65
  4735.4  330.07  4838.2  325.53    4874  324.11  4876.7  323.61    4880  324.11
  4937.9  324.11  4953.2  324.11  5037.6  324.11  5159.1  324.11  5237.1  324.11
  5315.9  324.11    5322  326.81  5336.8  327.18  5372.6  331.39  5468.8  339.12
  5534.4  343.46  5581.1  349.95  5625.4  353.28  5766.4   360.1  6011.8  389.89
#Mann= 13 ,-1 , 0
  3657.1     .12       0  3954.3     .16       0  4253.4     .12       0
  4838.2     .16       0    4874     .07       0    4880     .16       0
  4937.9     .05       0  4953.2     .07       0  5037.6     .05       0
  5159.1     .07       0  5237.1      .1       0  5336.8     .16       0
  5468.8     .12       0
Bank Sta=4594.1,5372.6
XS Rating Curve= 0 ,0
Exp/Cntr=0.3,0.1

Type RM Length L Ch R = 1 ,12225   ,261,261,261
BEGIN DESCRIPTION:
ANDING BRANCH 23.0
END DESCRIPTION:
XS GIS Cut Line= 4
       3674721.4     10743143.31      3674638.07     10742396.76
      3674183.21     10741445.37      3673846.38     10740848.12
#Sta/Elev= 30
  3239.3  403.41  3262.2  403.07  3389.5   395.3  3594.6   374.5  3724.2  368.35
  3762.6   366.1  3916.6  358.72  4023.6  357.27  4114.3  358.66    4286   340.9
    4460  331.46    4528  326.47  4585.2  325.03  4624.2  324.48  4652.5  327.12
  4726.5  325.58  4748.5  324.11  4751.2  323.61  4754.5  324.11  5289.3  324.11
    5315  326.45  5329.7     325    5338  326.02  5345.6   329.6  5360.9  330.66
  5432.3   343.1    5471  345.16  5550.7  346.64  5637.4  353.97  5730.7  357.65
#Mann= 9 ,-1 , 0
  3239.3     .12       0  3262.2     .16       0  3724.2     .12       0
  3762.6     .16       0  4726.5     .05       0  4748.5    .033       0
  4754.5     .05       0  5289.3     .16       0    5471     .12       0
Bank Sta=4460,5360.9
XS Rating Curve= 0 ,0
Exp/Cntr=0.3,0.1

Type RM Length L Ch R = 1 ,11964   ,429,429,429
BEGIN DESCRIPTION:
ANDING BRANCH 22.0
END DESCRIPTION:
XS GIS Cut Line= 3
      3675049.64     10741860.21      3674449.61     10741410.19
      3673849.59     10740810.17
#Sta/Elev= 30
  4252.3  369.13  4265.9  368.49  4274.2  366.41  4380.5  352.43  4388.8  352.18
  4402.3  349.42  4452.3   344.6  4502.3  338.08    4545  333.86  4559.6  334.11
  4565.9  332.38  4588.8  330.67  4638.8  326.43  4649.3  324.11  4652.1  323.61
  4655.3  324.11  4771.2  324.11  5418.1  324.11    5469  324.11  5497.3  325.04
  5508.1  326.52  5553.9  331.32    5568  331.86  5596.3  335.63  5610.5  335.71
  5638.7  339.74  5652.9   340.4  5723.6  348.91  5751.9  353.51  5850.9  360.26
#Mann= 6 ,-1 , 0
  4252.3     .16       0  4649.3    .033       0  4655.3     .16       0
  4771.2     .05       0  5418.1     .16       0  5508.1     .12       0
Bank Sta=4588.8,5553.9
XS Rating Curve= 0 ,0
Exp/Cntr=0.3,0.1
