--- BEAVER CREEK.prj (project) ---

Proj Title=BEAVER CREEK Base Level Engineering
Current Plan=p01
Default Exp/Contr=0.3,0.1
English Units
Geom File=g01
Geom File=g02
Flow File=f01
Plan File=p01
Y Axis Title=Elevation
X Axis Title(PF)=Main Channel Distance
X Axis Title(XS)=Station
BEGIN DESCRIPTION:
BEAVER CREEK
END DESCRIPTION:
DSS File=dss
DSS Export Rating Curves= 0
DSS Export Rating Curve Sorted= 0
DSS Export Volume Flow Curves= 0
DXF OffsetX= 0
DXF OffsetY= 0
DXF ScaleX= 1
DXF ScaleY= 10

--- BEAVER CREEK.p01 (plan) ---

Plan Title=Multiple Run
Program Version=4.10
Short Identifier=Multiple Run
Geom File=g01
Flow File=f01
Subcritical Flow
K Sum by GR= 0
Std Step Tol= 0.01
Critical Tol= 0.01
Num of Std Step Trials= 20
Max Error Tol= 0.3
Flow Tol Ratio= 0.001
Split Flow NTrial= 30
Split Flow Tol= 0.02
Split Flow Ratio= 0.02
Log Output Level= 0
Friction Slope Method= 1
Unsteady Friction Slope Method= 2
Unsteady Bridges Friction Slope Method= 1
Parabolic Critical Depth
Global Vel Dist= 1 , 1 , 1
Global Log Level= 0
CheckData=True
Encroach Param=-1 ,0,0, 0
BEGIN DESCRIPTION:
Multiple Run
END DESCRIPTION:
Computation Interval=1HOUR
Output Interval=1HOUR
Run HTab= 0
Run UNet= 0
Run PostProcess= 0
Run WQNet= 0
UNET Theta= 1
UNET Theta Warmup= 1
UNET ZTol= 0.02
UNET ZSATol= 0.05
UNET MxIter= 20
UNET MaxInSteps= 0
UNET DtIC= 0
UNET DtMin= 0
UNET MaxCRTS= 20
UNET WFStab= 2
UNET SFStab= 1
UNET WFX= 1
UNET SFX= 1
UNET DSS MLevel= 4
UNET DZMax Abort= 100
UNET Convert EG Bridges= 0
UNET Use Existing IB Tables=-1
UNET Froude Reduction=False
UNET Froude Limit= 1
UNET Froude Power= 10
UNET Time Slicing=0,0, 5
UNET Junction Losses=0
Instantaneous Interval=1HOUR
DSS File=dss
Write IC File= 0
Write IC File at Sim End=0
Echo Input=False
Echo Parameters=False
Echo Output=False
Write Detailed= 0
WQ AD Non Conservative
WQ ULTIMATE=-1
WQ Max Comp Step=1HOUR
WQ Output Interval=15MIN
WQ Output Selected Increments= 0
WQ Output face flow=0
WQ Output face velocity=0
WQ Output face area=0
WQ Output face dispersion=0
WQ Output cell volume=0
WQ Output cell surface area=0
WQ Output cell continuity=0
WQ Output cumulative cell continuity=0
WQ Output face conc=0
WQ Output face dconc_dx=0
WQ Output face courant=0
WQ Output face peclet=0
WQ Output face adv mass=0
WQ Output face disp mass=0
WQ Output cell mass=0
WQ Output cell source sink temp=0
WQ Output cell source sink nsm=0
WQ Output MaxMinRange=-1
WQ Daily Max Min Mean=-1
WQ Daily Range=0
WQ Daily Time=0
WQ Create Restart=0
WQ Fixed Restart=0
WQ System Summary=0
WQ Use Fixed Temperature=0
Sorting and Armoring Iterations= 10
XS Update Threshold= 0.02
Hydraulics Update Threshold= 0.02
Energy Slope Method= 1
Volume Change Method= 0
XS Weighting Method= 0
Number of US Weighted Cross Sections= 1
Number of DS Weighted Cross Sections= 1
Upstream XS Weight=0.25
Main XS Weight=0.5
Downstream XS Weight=0.25
Number of DS XS's Weighted with US Boundary= 1
Upstream Boundary Weight= 1
Weight of XSs Associated with US Boundary= 0
Number of US XS's Weighted with DS Boundary= 1
Downstream Boundary Weight= 0.5
Weight of XSs Associated with DS Boundary= 0.5
Sediment Output Level= 4
Mass or Volume Output= 0
Output Increment Type= 1
Profile and TS Output Increment= 10
XS Output Flag= 0
XS Output Increment= 10
Disregard all LS=0
Disregard all Conn=0
Disregard all Breaches=0
Disregard all Pumps=0

--- BEAVER CREEK.f01 (steady flow) ---

Flow Title=Multiple
Program Version=4.10
Number of Profiles= 7
Profile Names=10-year,25-year,50-year,1pct_min,100-year,1pct_plu,500-year
River Rch & RM=BEAVER CREEK,Reach-1         ,84360
     838    1175    1463    1340    1812    2451    2791
River Rch & RM=BEAVER CREEK,Reach-1         ,81706
     916    1286    1603    1469    1986    2686    3061
River Rch & RM=BEAVER CREEK,Reach-1         ,77913
    1341    1924    2433    2259    3055    4132    4838
River Rch & RM=BEAVER CREEK,Reach-1         ,77279
    1447    2076    2625    2435    3293    4453    5205
River Rch & RM=BEAVER CREEK,Reach-1         ,73879
    3184    4724    6111    5786    7824   10581   12890
River Rch & RM=BEAVER CREEK,Reach-1         ,72522
    3184    4724    6111    5786    7824   10581   12890
River Rch & RM=BEAVER CREEK,Reach-1         ,71600
    3356    4986    6454    6113    8267   11180   13633
River Rch & RM=BEAVER CREEK,Reach-1         ,70617
    3356    4986    6454    6113    8267   11180   13633
River Rch & RM=BEAVER CREEK,Reach-1         ,69071
    3399    5045    6525    6175    8351   11294   13748
River Rch & RM=BEAVER CREEK,Reach-1         ,66932
    3507    5201    6725    6361    8603   11634   14146
River Rch & RM=BEAVER CREEK,Reach-1         ,66845
    3507    5201    6725    6361    8603   11634   14146
River Rch & RM=BEAVER CREEK,Reach-1         ,63713
    3570    5285    6825    6445    8716   11787   14285
River Rch & RM=BEAVER CREEK,Reach-1         ,58657
    3648    5403    6979    6591    8914   12055   14615
River Rch & RM=BEAVER CREEK,Reach-1         ,57600
    4347    6472    8389    7948   10749   14537   17733
River Rch & RM=BEAVER CREEK,Reach-1         ,55177
    4352    6471    8380    7931   10726   14506   17659
River Rch & RM=BEAVER CREEK,Reach-1         ,50528
    4391    6513    8420    7955   10758   14549   17645
River Rch & RM=BEAVER CREEK,Reach-1         ,45971
    6580    9881   12884   12266   16589   22434   27622
River Rch & RM=BEAVER CREEK,Reach-1         ,41132
    6559    9834   12808   12179   16471   22275   27361
River Rch & RM=BEAVER CREEK,Reach-1         ,38972
    6485    9707   12629   11995   16221   21938   26883
River Rch & RM=BEAVER CREEK,Reach-1         ,38607
    6984   10459   13612   12930   17486   23648   28985
River Rch & RM=BEAVER CREEK,Reach-1         ,34911
    7357   11030   14365   13655   18467   24974   30649
River Rch & RM=BEAVER CREEK,Reach-1         ,31791
    7357   11030   14365   13655   18467   24974   30649
River Rch & RM=BEAVER CREEK,Reach-1         ,30954
    8058   12108   15797   15039   20338   27505   33854
River Rch & RM=BEAVER CREEK,Reach-1         ,30496
    8081   12135   15824   15057   20363   27539   33860
River Rch & RM=BEAVER CREEK,Reach-1         ,28408
    8030   12043   15691   14917   20173   27282   33485
River Rch & RM=BEAVER CREEK,Reach-1         ,27105
    8106   12158   15841   15059   20365   27542   33801
River Rch & RM=BEAVER CREEK,Reach-1         ,25683
    8106   12158   15841   15059   20365   27542   33801
River Rch & RM=BEAVER CREEK,Reach-1         ,25303
    8217   12316   16040   15241   20611   27875   34176
River Rch & RM=BEAVER CREEK,Reach-1         ,22971
    8253   12366   16100   15293   20683   27971   34273
River Rch & RM=BEAVER CREEK,Reach-1         ,20890
    8201   12274   15968   15155   20496   27719   33907
River Rch & RM=BEAVER CREEK,Reach-1         ,17511
    8332   12464   16210   15380   20800   28129   34384
River Rch & RM=BEAVER CREEK,Reach-1         ,14231
    8393   12550   16319   15479   20933   28310   34585
River Rch & RM=BEAVER CREEK,Reach-1         ,12090
    8350   12470   16200   15350   20760   28075   34230
River Rch & RM=BEAVER CREEK,Reach-1         ,8402
    8430   12590   16355   15497   20958   28344   34557
River Rch & RM=BEAVER CREEK,Reach-1         ,7709
    8430   12590   16355   15497   20958   28344   34557
River Rch & RM=BEAVER CREEK,Reach-1         ,7075
    8382   12505   16232   15369   20784   28108   34215
River Rch & RM=BEAVER CREEK,Reach-1         ,3703
    8282   12336   15995   15127   20457   27666   33598
Boundary for River Rch & Prof#=BEAVER CREEK,Reach-1         , 1
Up Type= 0
Dn Type= 3
Dn Slope=0.00046
Boundary for River Rch & Prof#=BEAVER CREEK,Reach-1         , 2
Up Type= 0
Dn Type= 3
Dn Slope=0.00046
Boundary for River Rch & Prof#=BEAVER CREEK,Reach-1         , 3
Up Type= 0
Dn Type= 3
Dn Slope=0.00046
Boundary for River Rch & Prof#=BEAVER CREEK,Reach-1         , 4
Up Type= 0
Dn Type= 3
Dn Slope=0.00046
Boundary for River Rch & Prof#=BEAVER CREEK,Reach-1         , 5
Up Type= 0
Dn Type= 3
Dn Slope=0.00046
Boundary for River Rch & Prof#=BEAVER CREEK,Reach-1         , 6
Up Type= 0
Dn Type= 3
Dn Slope=0.00046
Boundary for River Rch & Prof#=BEAVER CREEK,Reach-1         , 7
Up Type= 0
Dn Type= 3
Dn Slope=0.00046
DSS Import GetInterval= 0
DSS Import GetPeak= 0
DSS Import FillOption= 0

--- BEAVER CREEK.g01 (geometry) ---

Geom Title=Existing Conditions
Program Version=4.10

River Reach=BEAVER CREEK    ,Reach-1
Reach XY= 30
      3731207.39      10706960.9       3728219.5       10703440.
        3726879.       10702934.      3725319.25       10699757.
      3721744.25       10696304.       3721498.5       10695028.
       3717019.5       10691700.      3716612.25       10690715.
        3712259.       10689311.        3709041.       10690091.
      3708198.75       10689291.      3706249.25       10689786.
      3704443.25       10685289.        3702853.       10684034.
      3702481.75       10682914.      3698084.25       10678031.
      3695446.75       10677766.       3690962.5       10675170.
      3690589.25       10673861.      3689135.25       10672953.
        3688819.       10671811.      3687650.25       10671704.
       3686522.5       10670844.        3686212.       10669844.
        3683872.       10667445.      3681123.25       10667033.
        3680896.       10666348.      3679449.75       10665850.
       3678975.5       10667647.        3678102.       10668182.

Type RM Length L Ch R = 1 ,84360   ,440,440,440
BEGIN DESCRIPTION:
BEAVER CREEK 139.0
END DESCRIPTION:
XS GIS Cut Line= 3
       3731099.6      10706610.2      3730849.61     10706810.19
      3730799.61      10707160.2
#Sta/Elev= 30
  4670.8  490.59    4674  490.59    4678  494.23  4684.4   493.5  4698.8  490.57
  4713.2  486.33  4721.2  482.69  4734.8  479.86  4762.8  479.68  4770.8  480.74
  4791.6  479.72  4798.8  481.97    4806  480.96  4820.5   476.1  4913.3  466.51
  4934.1   465.1  5008.1  464.35  5010.9  463.85  5014.1  464.35  5071.8   464.9
    5092  466.99  5132.4   469.8    5193  476.75  5223.3  477.08  5233.4  479.84
  5243.5  478.83  5273.8   484.2    5294  486.29  5314.2  485.94  5344.5  488.64
#Mann= 3 ,-1 , 0
  4670.8     .16       0  5008.1     .07       0  5014.1     .16       0
Bank Sta=4913.3,5092
XS Rating Curve= 0 ,0
Exp/Cntr=0.3,0.1

Type RM Length L Ch R = 1 ,83920   ,429,429,429
BEGIN DESCRIPTION:
BEAVER CREEK 138.0
END DESCRIPTION:
XS GIS Cut Line= 3
      3730999.63     10706210.17      3730599.61     10706510.19
      3730199.64      10706410.2
#Sta/Elev= 30
  4487.4  501.58  4494.7  499.78  4537.4  497.06  4635.1  483.67  4659.3   480.4
  4680.1  479.18  4687.4  475.39  4715.5  475.46  4730.1  470.72  4737.4  470.18
    4751  471.56    4760  470.31    4801  465.86  4859.3  461.71  4909.3  459.92
    4990  460.24  4994.7  455.82  4997.5  455.32  5000.7  455.82  5005.5  459.46
  5010.6  460.26    5039  462.85  5080.2  464.03  5183.3  461.17  5216.8  462.73
    5276  469.57  5286.3  469.18  5335.3  475.99  5348.2   476.7  5399.7   485.3
#Mann= 5 ,-1 , 0
  4487.4     .16       0  4635.1     .05       0    4760     .16       0
  4994.7     .07       0  5000.7     .16       0
Bank Sta=4990,5010.6
XS Rating Curve= 0 ,0
Exp/Cntr=0.3,0.1

Type RM Length L Ch R = 1 ,83491   ,409,409,409
BEGIN DESCRIPTION:
BEAVER CREEK 137.0
END DESCRIPTION:
XS GIS Cut Line= 3
      3730849.61     10706160.19      3730449.61     10706160.19
      3730249.61     10706260.19
#Sta/Elev= 30
  4594.4  483.28  4614.4  480.84  4644.4  478.65  4651.4  477.39  4684.4   474.1
  4704.4  471.09  4724.4  469.42  4734.4  469.15  4744.4  467.84  4754.4  467.47
  4764.4  466.35  4844.4  463.36  4907.1  462.91  4924.4  462.56  4954.4  459.86
  5002.8   456.6  5005.4  454.69  5008.1  454.19  5011.4  454.69  5030.7  457.29
  5039.1  459.95  5047.5  459.87  5106.2  467.17  5114.6  468.73  5128.6  469.57
  5136.9  471.43  5173.3  474.69  5195.6   477.7  5209.6   480.5    5218  480.87
#Mann= 5 ,-1 , 0
  4594.4     .16       0  4651.4     .05       0  4907.1     .16       0
  5005.4     .07       0  5011.4     .16       0
Bank Sta=4954.4,5039.1
XS Rating Curve= 0 ,0
Exp/Cntr=0.3,0.1

Type RM Length L Ch R = 1 ,83082   ,412,412,412
BEGIN DESCRIPTION:
BEAVER CREEK 136.0
END DESCRIPTION:
XS GIS Cut Line= 3
      3730549.59     10705410.21      3730249.61     10705810.19
      3730149.59      10705860.2
#Sta/Elev= 30
  4510.2  497.23    4532  497.74  4538.3  496.01  4546.6  497.37  4552.9  495.41
  4560.2   495.5  4567.5  493.78  4573.7  490.28    4582  489.63  4588.3  486.96
  4617.5  481.23    4632  475.79  4646.6  472.02  4710.2  462.98  4736.4  460.76
  4760.2  458.65    4782  459.08  4788.3  457.24  4802.9  456.06  4885.6  455.96
  4917.5  456.07    4982     453  4993.6  451.13  4996.4  450.63  4999.6  451.13
    5007  452.98    5013  452.98  5054.9  459.47  5085.6  465.45    5122  469.43
#Mann= 5 ,-1 , 0
  4510.2     .16       0  4736.4     .05       0  4885.6     .16       0
  4993.6     .07       0  4999.6     .16       0
Bank Sta=4982,5007
XS Rating Curve= 0 ,0
Exp/Cntr=0.3,0.1

Type RM Length L Ch R = 1 ,82670   ,536,536,536
BEGIN DESCRIPTION:
BEAVER CREEK 135.0
END DESCRIPTION:
XS GIS Cut Line= 3
      3730499.56     10705410.19      3730099.61     10705460.19
       3729999.6      10705560.2
#Sta/Elev= 30
  4639.7  488.14  4649.7  487.18  4659.8  484.84  4669.9     484  4677.4  481.94
  4682.5  481.83  4700.1  478.02  4720.3  475.06  4750.5  472.39  4763.1  469.24
  4851.3  461.46  4861.4  459.93  4872.5  459.89  4911.8  454.48  4919.3  453.95
  4931.9  454.47  4952.1  452.73  4962.1  451.09  4972.2  451.36  4982.3  450.16
  4992.4     450  4996.9  448.83  4999.7  448.33  5002.9  448.83    5005  449.62
  5045.8  449.75    5071  451.93  5099.3  456.01    5170   463.9  5184.2  464.38
#Mann= 5 ,-1 , 0
  4639.7     .16       0  4872.5     .05       0  4996.9     .04       0
  5002.9     .05       0  5045.8     .16       0
Bank Sta=4992.4,5005
XS Rating Curve= 0 ,0
Exp/Cntr=0.3,0.1

Type RM Length L Ch R = 1 ,82134   ,428,428,428
BEGIN DESCRIPTION:
BEAVER CREEK 134.0
END DESCRIPTION:
XS GIS Cut Line= 3
       3729899.6     10704760.21      3729749.61     10705110.19
      3729699.61     10705360.17
#Sta/Elev= 30
  4626.3  485.41  4635.3  484.22  4640.8  485.19  4658.9  483.14  4669.8  480.53
  4680.7  479.65  4702.4  474.33  4711.5  473.35  4724.2  469.95  4756.8  467.27
  4800.4   461.6    4833  459.56  4840.2  457.74  4869.3  455.61  4906.6  451.33
  4930.9  449.22  4952.7   446.3  4963.5   446.3  4982.3  444.13  4985.1  443.63
  4988.3  444.13  5004.3  446.05  5027.5  446.35  5059.3   449.5  5078.5  451.35
  5088.7  453.48  5119.2  455.64  5139.6   458.5    5211  465.07    5262  471.21
#Mann= 5 ,-1 , 0
  4626.3     .16       0  4906.6     .05       0  4982.3     .04       0
  4988.3     .05       0  5059.3     .16       0
Bank Sta=4963.5,5004.3
XS Rating Curve= 0 ,0
Exp/Cntr=0.3,0.1

Type RM Length L Ch R = 1 ,81706   ,70,70,70
BEGIN DESCRIPTION:
BEAVER CREEK 133.0
END DESCRIPTION:
XS GIS Cut Line= 4
      3729775.41     10704582.34      3729623.48     10704727.76
      3729278.43     10705020.73      3728893.34     10705401.48
#Sta/Elev= 30
  4443.8  472.45  4460.6  470.23  4467.5  471.69  4495.8  470.09    4503   468.2
  4552.4  469.37  4587.9   467.7  4594.9     467  4602.1  463.05    4609  465.34
  4616.2  464.74  4686.5  456.01  4694.2  453.54  4715.1  453.99  4722.8  451.84
  4793.1  447.28    4949  446.23  4996.6  444.97  4999.4  444.47  5002.6  444.97
  5013.4  446.03  5034.7   446.1  5140.9     458  5197.5  461.45  5232.8  460.87
  5310.6   454.5    5452  455.65  5558.1  460.77  5642.9  468.44  5648.3  470.69
#Mann= 3 ,-1 , 0
  4443.8     .05       0  4996.6     .04       0  5002.6     .05       0
Bank Sta=4949,5013.4
XS Rating Curve= 0 ,0
Exp/Cntr=0.3,0.1

Type RM Length L Ch R = 1 ,81636   ,352,352,352
BEGIN DESCRIPTION:
Mapping XS c25f8cee
END DESCRIPTION:
XS GIS Cut Line= 5
      3729749.31     10704495.59      3729402.12     10704831.92
      3729226.34     10704975.15      3728985.46     10705213.87
      3728837.86     10705374.49
#Sta/Elev= 30
  4386.4  479.13  4396.6  480.35  4403.5  478.07  4410.7  480.37  4417.7  476.31
  4424.9  477.35  4469.8   470.7  4502.6   466.1  4686.5  454.23  4693.4  451.55
  4885.1   445.7  4960.3  443.96  4963.1  443.46  4966.3  443.96  5048.1  445.84
  5074.3  448.58  5111.8  451.88  5175.6  457.33  5302.9  451.44  5408.9     453
  5536.4  460.66  5543.2  464.09  5564.8  464.16  5571.6  467.64    5579  464.02
  5585.8  468.12    5600   470.3  5614.1  467.63  5620.9  472.12  5653.8  474.78
#Mann= 6 ,-1 , 0
  4386.4     .12       0  4469.8     .05       0  4960.3     .04       0
  4966.3     .05       0  5074.3     .16       0  5111.8     .05       0
Bank Sta=4885.1,5048.1
XS Rating Curve= 0 ,0
Exp/Cntr=0.3,0.1

Type RM Length L Ch R = 1 ,81284   ,476,476,476
BEGIN DESCRIPTION:
BEAVER CREEK 132.0
END DESCRIPTION:
XS GIS Cut Line= 3
      3729249.61     10704410.18      3729049.61     10704710.19
      3728699.63     10705060.16
#Sta/Elev= 30
  4640.2  460.44  4668.8  459.65  4704.8  456.71  4748.4   451.8  4755.9  449.88
  4770.9   448.6  4776.9  447.18  4784.4  446.98  4791.9  445.11    4807  444.58
  4820.5  442.52    4843  440.95  4856.5  441.29  4870.1  439.79  4915.1  439.76
  4942.2  438.67  4951.2  439.25  4994.8  437.58  4997.5  437.08  5000.8  437.58
    5029  439.05  5133.7  441.56  5184.6  444.92  5269.5  452.44  5316.2  455.31
  5396.7   462.9  5439.2  468.07  5453.3  470.83  5481.6  474.46  5495.7  475.53
#Mann= 5 ,-1 , 0
  4640.2     .16       0  4994.8     .07       0  5000.8     .16       0
  5133.7     .12       0  5316.2     .16       0
Bank Sta=4951.2,5029
XS Rating Curve= 0 ,0
Exp/Cntr=0.3,0.1

Type RM Length L Ch R = 1 ,80808   ,453,453,453
BEGIN DESCRIPTION:
BEAVER CREEK 131.0
END DESCRIPTION:
XS GIS Cut Line= 3
      3729149.63     10704010.17      3728749.61     10704360.19
       3728399.6     10704410.19
#Sta/Elev= 30
  4483.5  474.96  4496.1  474.21  4504.9  473.75  4511.5  472.08  4519.1  468.06
  4603.6  461.61  4625.4  457.95  4632.1  455.55  4639.4  455.21  4646.3  454.21
  4674.8  453.81  4688.7  451.86  4709.9   450.7    4746  446.11  4820.8  439.69
  4901.6   435.9  4955.6  432.29  4958.3  431.79  4961.6  432.29  4979.4  433.63
  5025.1  433.58  5045.3  435.55  5085.8  440.62    5106  441.82  5116.1  444.04
  5166.6  449.16  5196.9   453.9  5247.4  457.83    5300   464.1  5368.6  471.08
#Mann= 8 ,-1 , 0
  4483.5     .05       0  4496.1     .16       0  4639.4     .12       0
  4688.7     .16       0  4820.8     .12       0  4955.6     .07       0
  4961.6     .12       0    5300     .16       0
Bank Sta=4901.6,5045.3
XS Rating Curve= 0 ,0
Exp/Cntr=0.3,0.1

Type RM Length L Ch R = 1 ,80355   ,469,469,469
BEGIN DESCRIPTION:
BEAVER CREEK 130.0
END DESCRIPTION:
XS GIS Cut Line= 3
      3728899.61     10703710.19      3728499.61     10704010.19
       3728399.6     10704160.21
#Sta/Elev= 30
  4494.7  468.82  4531.2  464.99    4552  461.04    4557  461.62  4587.4  459.84
  4616.6  456.08  4637.4  454.93  4666.6  451.37  4694.7  449.16  4708.2  446.75
  4737.4  444.35    4752  442.05  4772.8   441.4  4816.6  436.24  4872.8   432.2
  4931.2  431.76  4944.7  430.75  4955.2  427.81    4958  427.31  4961.2  427.81
  4987.4  429.29  4991.6  428.15  5015.8  428.38  5030.8  431.01  5053.3   433.3
  5074.3  434.78  5080.3  436.47  5102.9  439.29  5130.7  441.75    5175  447.89
#Mann= 6 ,-1 , 0
  4494.7     .05       0    4557     .12       0  4955.2     .07       0
  4961.2     .12       0  5015.8     .16       0  5130.7     .12       0
Bank Sta=4931.2,5053.3
XS Rating Curve= 0 ,0
Exp/Cntr=0.3,0.1

Type RM Length L Ch R = 1 ,79886   ,456,456,456
BEGIN DESCRIPTION:
BEAVER CREEK 129.0
END DESCRIPTION:
XS GIS Cut Line= 3
      3728549.63     10703360.17      3728299.61     10703610.19
      3728099.61     10703960.19
#Sta/Elev= 30
  4641.3  456.08  4655.5  455.46  4757.2  446.39  4825.2  437.61  4839.3  436.88
  4895.9   430.5    4910  430.14  4924.2  428.37  4980.7  425.85  4999.8  424.25
  5002.6  423.75  5005.8  424.25  5024.4  425.88  5098.5  427.25  5110.8  428.59
  5120.9     428  5125.8   428.7  5179.2  432.27  5185.6  433.86  5207.2  435.27
  5236.3  439.54  5259.8  442.05  5266.3  443.74  5282.1  445.14  5303.7  448.77
  5340.4  452.69  5352.6   455.2  5362.7  455.59  5390.1  460.99    5398  461.14
#Mann= 6 ,-1 , 0
  4641.3     .12       0  4757.2     .16       0  4999.8     .07       0
  5005.8     .16       0  5125.8     .05       0  5236.3     .12       0
Bank Sta=4924.2,5110.8
XS Rating Curve= 0 ,0
Exp/Cntr=0.3,0.1

Type RM Length L Ch R = 1 ,79430   ,401,401,401
BEGIN DESCRIPTION:
BEAVER CREEK 128.0
END DESCRIPTION:
XS GIS Cut Line= 3
      3727999.61     10702960.21      3727999.61     10703310.19
      3727899.61      10703710.2
#Sta/Elev= 30
  4648.7  439.86  4688.7  437.56  4698.7  435.93  4708.7  435.25  4719.2  433.04
  4778.7  425.16  4818.7  422.02  4858.7  421.82  4868.7  422.86  4908.7  424.46
  4928.7  423.41  4948.7  423.91  4968.7  422.09  4993.2  421.43  4995.9  420.93
  4999.2  421.43  5011.4  422.94  5021.9  423.61  5057.9   422.9  5091.4  423.67
  5112.1   425.4  5140.4  425.55  5145.6  426.46  5173.9  427.22  5186.8  428.51
    5228  430.02  5297.6  434.06  5346.6  437.63  5359.5  439.36    5411  442.68
#Mann= 5 ,-1 , 0
  4648.7     .12       0  4719.2     .16       0  4993.2     .07       0
  4999.2     .16       0  5011.4     .12       0
Bank Sta=4948.7,5021.9
XS Rating Curve= 0 ,0
Exp/Cntr=0.3,0.1

Type RM Length L Ch R = 1 ,79029   ,568,568,568
BEGIN DESCRIPTION:
Mapping XS 9d8586aa
END DESCRIPTION:
XS GIS Cut Line= 3
      3727827.94     10702620.64      3727459.89     10703828.94
      3727626.56     10704759.52
#Sta/Elev= 30
  4417.2  460.39  4463.4  457.35  4527.9  446.75  4599.9  434.67  4698.5  426.92
  4779.6  420.82  4782.4  420.32  4785.6  420.82    4903   421.5  5135.7  420.82
  5255.3  422.59  5294.8  426.37  5347.1  430.44  5457.3     444  5566.6  457.64
  5646.2  464.38  5721.1  470.38  5854.3  480.79  5925.4  481.83  5943.4  478.75
  5976.2  473.13  5991.1  473.79  5996.5   471.1  6037.1  464.73  6087.9  459.65
  6103.6  456.37  6162.5  454.75  6216.2  449.86  6387.7  446.87  6625.7  455.04
#Mann= 10 ,-1 , 0
  4417.2     .12       0  4527.9     .16       0  4779.6    .033       0
  4785.6     .16       0    4903     .05       0  5135.7     .16       0
  5457.3     .12       0  5646.2     .16       0  5721.1     .12       0
  5943.4     .16       0
Bank Sta=4698.5,5294.8
XS Rating Curve= 0 ,0
Exp/Cntr=0.3,0.1

Type RM Length L Ch R = 1 ,78461   ,548,548,548
BEGIN DESCRIPTION:
Mapping XS 70969a17
END DESCRIPTION:
XS GIS Cut Line= 3
      3727730.74     10702453.92      3726966.84     10703162.27
      3726620.06     10704486.95
#Sta/Elev= 30
  4155.6  465.28  4160.7  464.69  4211.9   460.6  4245.7  458.04  4259.9  454.68
  4266.7  455.47  4373.3  438.79  4466.8   428.4  4493.5  426.28  4578.5  421.44
  4624.9  420.82  4627.6  420.32  4630.9  420.82  4677.4  420.82  5867.1  420.82
  5931.7  424.79  5955.7  426.23    5991  427.96  5996.1  429.92  6031.4  430.84
  6042.9  432.76  6063.5  432.95  6129.2  437.82  6149.2  439.32  6309.1  451.09
  6386.8  453.04  6404.7  450.82  6470.8  449.61  6497.7  451.14  6566.7  451.34
#Mann= 11 ,-1 , 0
  4155.6     .12       0  4160.7     .16       0  4211.9     .12       0
  4466.8     .16       0  4624.9    .033       0  4630.9     .16       0
  4677.4     .05       0  5931.7     .16       0  6129.2     .05       0
  6149.2     .16       0  6386.8     .05       0
Bank Sta=4493.5,5955.7
XS Rating Curve= 0 ,0
Exp/Cntr=0.3,0.1

Type RM Length L Ch R = 1 ,77913   ,41,41,41
BEGIN DESCRIPTION:
BEAVER CREEK 125.0
END DESCRIPTION:
XS GIS Cut Line= 3
      3727226.81     10702404.03      3726177.36     10702979.54
      3725818.55     10703325.32
#Sta/Elev= 30
  4423.8  437.24  4500.4  430.08  4580.3  426.67  4657.4  420.82  4660.1  420.32
  4663.4  420.82  4780.2  420.82  4817.3  420.82  5377.9  422.26  5388.8  420.82
  5427.2  421.52  5443.3  423.85    5449  420.82  5465.1  423.53    5472  422.29
  5515.5  427.43  5524.8  430.62  5530.5  429.94  5546.6   435.6  5587.3  441.74
  5722.1  452.27  5768.2  455.57  5824.8  453.96  5845.9  451.28  5862.9  452.41
  5864.9  452.59  5874.2  451.74  5881.4  453.97  5973.2  461.01    6119  462.64
#Mann= 11 ,-1 , 0
  4423.8     .05       0  4657.4    .033       0  4663.4     .05       0
  4780.2     .12       0  4817.3     .05       0  5388.8      .1       0
    5472     .05       0  5587.3     .12       0  5722.1     .16       0
  5862.9     .12       0  5864.9     .05       0
Bank Sta=4580.3,5515.5
XS Rating Curve= 0 ,0
Exp/Cntr=0.3,0.1

Type RM Length L Ch R = 1 ,77872   ,91,91,91
BEGIN DESCRIPTION:
Mapping XS 8096dad9
END DESCRIPTION:
XS GIS Cut Line= 2
      3727178.68     10702377.96      3726194.41     10702929.99
#Sta/Elev= 30
  4451.7  435.71  4591.5  426.32  4607.5  427.53  4613.2  424.24  4663.8  422.23
  4666.6  421.73  4669.8  422.23  4710.2   424.7  4747.8  426.29  4752.6   424.2
  4769.5  426.32  4840.5  425.16  4885.4  426.29  5216.5  425.46  5260.4  425.93
    5283  424.63  5288.8  426.33  5348.1   426.3    5364  423.65  5369.8  426.21
  5385.7  424.03  5391.5  426.84  5423.4  427.61    5448  426.12  5448.4  426.19
  5482.5  427.09  5531.8  435.43  5539.8  439.52  5564.4  442.16  5580.2  443.82
#Mann= 10 ,-1 , 0
  4451.7     .05       0  4663.8     .03       0  4669.8     .05       0
  4752.6     .12       0  4885.4     .05       0  5216.5     .16       0
  5260.4     .05       0    5448      .1       0  5448.4     .05       0
  5564.4     .16       0
Bank Sta=4613.2,4710.2
XS Rating Curve= 0 ,0
Exp/Cntr=0.3,0.1

Type RM Length L Ch R = 1 ,77781   ,502,502,502
BEGIN DESCRIPTION:
BEAVER CREEK 124.0
END DESCRIPTION:
XS GIS Cut Line= 2
       3727143.5     10702311.57      3726152.98     10702831.53
#Sta/Elev= 30
  4446.7  441.33  4516.1  437.02  4521.8  435.39  4597.9  432.01    4610   427.5
    4632  422.45  4664.8  421.52  4699.6  425.16  4729.6  420.06    4753  414.16
  4789.9  412.03  4802.8  409.73  5031.5  405.63  5039.7  406.47  5094.6  404.98
  5122.3  406.25  5155.5  404.21  5193.5   400.9  5196.3   400.4  5199.5   400.9
    5228  403.27  5248.9  403.58  5264.3  406.04  5343.3  418.09  5424.5  425.85
  5447.4  428.63  5478.9  435.78  5491.5   435.8  5513.6  440.66  5565.4  446.44
#Mann= 8 ,-1 , 0
  4446.7     .05       0  4729.6     .12       0  5031.5     .05       0
  5155.5     .12       0  5193.5     .07       0  5199.5     .12       0
    5228     .16       0  5424.5     .05       0
Bank Sta=5039.7,5264.3
XS Rating Curve= 0 ,0
Exp/Cntr=0.3,0.1

Type RM Length L Ch R = 1 ,77279   ,412,412,412
BEGIN DESCRIPTION:
BEAVER CREEK 123.0
END DESCRIPTION:
XS GIS Cut Line= 3
      3726849.63     10702060.19      3726449.61     10702110.19
       3726199.6      10702260.2
#Sta/Elev= 30
  4582.9  428.17  4597.5  425.52  4663.5  414.55  4673.6  414.15  4697.7  409.79
  4713.9  408.46    4724  406.09  4754.2  402.28  4794.6  400.53  4804.6  399.57
  4867.6  398.18  4922.6  397.92  4925.3  397.42  4928.6  397.92  4943.2  398.56
  5079.3  398.14    5089   399.9  5094.9  399.23  5102.7  400.96  5116.3  401.63
  5131.8  404.11    5161  407.15  5168.7  408.91  5219.3  414.02    5227  416.11
  5242.6  417.95  5254.3  421.31  5269.8  423.59  5274.7  426.18  5277.6  426.18
#Mann= 5 ,-1 , 0
  4582.9     .12       0  4597.5     .16       0  4697.7     .12       0
  4922.6     .07       0  4928.6     .12       0
Bank Sta=4794.6,5102.7
XS Rating Curve= 0 ,0
Exp/Cntr=0.3,0.1

Type RM Length L Ch R = 1 ,76867   ,438,438,438
BEGIN DESCRIPTION:
BEAVER CREEK 122.0
END DESCRIPTION:
XS GIS Cut Line= 3
      3727049.61     10702010.19      3726299.61     10701710.19
       3726099.6      10702060.2
#Sta/Elev= 30
  4222.8  448.04  4262.6  444.85  4286.1  442.58  4291.5  440.51    4309  440.31
    4352  434.19  4482.6  421.55  4501.5  418.33  4506.9  418.73  4524.4  415.73
  4553.2  413.23  4638.8  404.48  4707.5  401.56  4803.2  398.11  4812.2  396.91
  4814.9  396.41  4818.2  396.91  4868.1  396.91  5139.7  396.91  5214.9  396.91
  5258.8  398.37  5286.1  401.29    5330  405.78  5339.4  408.86  5345.1  408.16
  5353.1  409.84  5367.2  410.41  5425.8  417.12  5430.8  420.56  5433.7  420.56
#Mann= 10 ,-1 , 0
  4222.8     .16       0  4262.6     .12       0    4352     .16       0
  4553.2     .12       0  4803.2     .16       0  4812.2    .033       0
  4818.2     .16       0  4868.1     .05       0  5139.7     .12       0
  5367.2     .16       0
Bank Sta=4707.5,5286.1
XS Rating Curve= 0 ,0
Exp/Cntr=0.3,0.1

Type RM Length L Ch R = 1 ,76429   ,427,427,427
BEGIN DESCRIPTION:
BEAVER CREEK 121.0
END DESCRIPTION:
XS GIS Cut Line= 3
      3726499.62     10700960.18      3726099.61     10701360.19
       3725349.6      10701860.2
#Sta/Elev= 30
  4453.1  431.86  4523.8  423.53    4562  416.93  4594.5  414.18  4679.4  403.25
  4718.8  396.91  4721.6  396.41  4724.8  396.91  4736.2  396.91  5298.9  396.91
    5398  396.91  5487.5  396.91    5495  398.39  5546.1  401.01  5631.6  406.55
  5675.3  412.85  5696.3  417.86  5703.9  421.62  5717.4  424.08  5739.9  430.56
  5747.4  434.05  5768.5  435.02    5776  437.74  5798.8   442.5  5804.5  442.82
  5819.5  447.62  5825.5  447.13  5834.6  449.16  5861.6   456.6  5920.2  465.88
#Mann= 9 ,-1 , 0
  4453.1     .12       0    4562     .16       0  4718.8    .033       0
  4724.8     .16       0  4736.2     .05       0  5298.9     .16       0
    5398     .12       0  5631.6     .16       0  5798.8     .12       0
Bank Sta=4679.4,5546.1
XS Rating Curve= 0 ,0
Exp/Cntr=0.3,0.1

Type RM Length L Ch R = 1 ,76002   ,433,433,433
BEGIN DESCRIPTION:
BEAVER CREEK 120.0
END DESCRIPTION:
XS GIS Cut Line= 3
      3726249.57     10700660.22      3725849.61     10701010.19
      3725199.61     10701660.19
#Sta/Elev= 30
  4467.2  420.96  4495.1  421.15  4523.6  418.65  4573.5  416.95  4594.8  414.47
  4601.5  412.45  4615.7  411.26  4644.2  405.39    4666  403.64  4676.4   401.8
  4676.6  401.78  4686.9   400.9  4693.5  399.03  4712.3  396.91  4715.1  396.41
  4718.3  396.91    5375  396.91  5479.5  400.11  5493.6  401.62  5564.3  408.99
  5592.6  412.74  5622.3  418.17    5734  437.79  5748.2  441.36  5762.3  442.67
    5826  452.37  5847.2  455.78  5861.3  456.67  5889.6  462.78  5917.9  465.54
#Mann= 8 ,-1 , 0
  4467.2     .05       0  4676.4     .16       0  4676.6     .05       0
  4712.3    .033       0  4718.3     .05       0    5375     .12       0
  5622.3     .16       0    5826     .12       0
Bank Sta=4686.9,5493.6
XS Rating Curve= 0 ,0
Exp/Cntr=0.3,0.1

Type RM Length L Ch R = 1 ,75569   ,478,478,478
BEGIN DESCRIPTION:
Mapping XS 6673f89c
END DESCRIPTION:
XS GIS Cut Line= 5
      3726145.83     10700197.36      3725928.79      10700275.5
      3725820.28     10700449.11      3725598.93     10700661.78
      3725203.18     10700756.93
#Sta/Elev= 30
  4263.3  429.48  4269.9  425.52  4280.5  424.52  4286.1  422.44  4347.5  416.54
  4354.9  413.39  4365.6  412.34  4372.9  409.97  4403.6  405.97    4440  403.38
  4474.1  403.69  4561.4  409.61  4570.3  408.84  4592.1  410.06    4641  415.44
  4655.8  415.62    4714  414.59  4742.3  411.41  4760.3  406.06  4777.8  401.55
  4784.7  401.84    4810  396.91  4812.8  396.41    4816  396.91  5222.7  396.91
  5235.3  396.92  5272.1  401.29  5395.8  420.46  5408.2  424.02  5412.7  426.73
#Mann= 6 ,-1 , 0
  4263.3     .12       0  4474.1     .16       0  4760.3     .05       0
    4810    .033       0    4816     .05       0  5222.7     .12       0
Bank Sta=4784.7,5272.1
XS Rating Curve= 0 ,0
Exp/Cntr=0.3,0.1

Type RM Length L Ch R = 1 ,75091   ,31,31,31
BEGIN DESCRIPTION:
Mapping XS e2744cc0
END DESCRIPTION:
XS GIS Cut Line= 4
      3726134.96     10700051.97      3725939.64     10700062.82
      3725440.51     10700203.88      3724978.31     10700464.28
#Sta/Elev= 30
  4259.9  420.24  4265.3  418.26  4319.1  413.56  4325.3  411.84  4462.5  400.65
  4517.9  398.81  4577.5  401.11  4590.6  398.63    4595  398.59  4678.9  396.76
  4681.7  396.26  4684.9  396.76  4794.2  399.36  4860.8  396.91  4912.2  396.91
  5111.7  396.91  5146.4  396.91  5221.7  396.91  5234.4  398.47  5237.6  399.16
  5296.6   407.1  5302.6  409.69  5318.5  410.73  5367.6  419.24    5377   419.7
  5434.3  432.05  5442.8   432.6  5464.4  437.54  5470.2  440.34  5504.7  446.46
#Mann= 9 ,-1 , 0
  4259.9     .12       0  4577.5     .16       0    4595      .1       0
  4678.9     .03       0  4684.9      .1       0  4912.2     .05       0
  5111.7     .12       0  5146.4     .16       0  5234.4     .12       0
Bank Sta=4590.6,5237.6
XS Rating Curve= 0 ,0
Exp/Cntr=0.3,0.1

Type RM Length L Ch R = 1 ,75060   ,67,67,67
BEGIN DESCRIPTION:
Mapping XS bbde77fe
END DESCRIPTION:
XS GIS Cut Line= 3
      3726128.44     10699928.27      3725392.76     10700193.03
      3724973.19     10700430.94
#Sta/Elev= 30
  4234.9  416.01  4313.9  409.43  4499.4  398.69  4531.2  397.79  4557.9  399.48
  4632.7  396.35  4635.5  395.85  4638.7  396.35  4728.2  397.92  4743.8  398.46
    4882  402.29  4984.5  401.95  4989.7  401.83  5097.9  401.55  5157.8  401.42
  5163.6  399.08  5179.5  401.47  5185.2  400.23  5192.8  401.53  5228.5  400.94
  5296.3  405.19  5362.7  416.09  5368.4  418.36  5399.7   421.6  5405.9  424.15
  5443.4  429.42  5457.2  434.18  5480.2  436.65  5492.5  441.22  5499.1  441.82
#Mann= 8 ,-1 , 0
  4234.9     .12       0  4557.9     .16       0  4632.7     .03       0
  4638.7     .16       0  4728.2      .1       0  4984.5     .12       0
  4989.7     .05       0  5097.9     .12       0
Bank Sta=4499.4,4743.8
XS Rating Curve= 0 ,0
Exp/Cntr=0.3,0.1

Type RM Length L Ch R = 1 ,74993   ,683,683,683
BEGIN DESCRIPTION:
Mapping XS 7406c0a2
END DESCRIPTION:
XS GIS Cut Line= 4
      3725879.95     10699913.71       3725615.6     10700040.02
        3725363.     10700132.47      3724934.86      10700405.4
#Sta/Elev= 30
  4464.4  402.28  4582.5  393.51  4661.6   403.1  4701.4  405.99  4757.4  405.13
  4770.7  401.93  4776.1   403.3  4785.1  400.59  4831.8  396.94    4898  387.63
  4943.2  384.17  4948.5  387.68  4959.4  385.49  4973.7  381.95  5009.6  382.99
  5022.5  381.14  5025.3  380.64  5028.5  381.14  5049.1   381.3    5055  383.67
  5064.3  382.48  5070.3  384.48  5085.5   382.7  5100.7  384.37  5106.7  387.15
  5137.1  386.76  5185.4  390.45  5346.2  410.09  5491.7  433.19  5534.1  444.28
#Mann= 6 ,-1 , 0
  4464.4     .12       0  4661.6     .16       0    4898      .1       0
  4959.4     .12       0  5022.5     .07       0  5028.5     .12       0
Bank Sta=4948.5,5106.7
XS Rating Curve= 0 ,0
Exp/Cntr=0.3,0.1

Type RM Length L Ch R = 1 ,74310   ,75,75,75
BEGIN DESCRIPTION:
BEAVER CREEK 116.0
END DESCRIPTION:
XS GIS Cut Line= 3
       3725199.6      10699510.2      3725049.61     10699710.19
      3724899.61      10700110.2
#Sta/Elev= 30
  4777.6  404.72    4814  403.57  4838.8   398.6  4877.6  391.03  4920.3  386.51
  4955.7  380.89    4964  375.91  4970.3  376.07  4977.6  373.23  4988.1  372.66
  4990.9  372.16  4994.1  372.66  5005.7  373.34  5024.5  376.27  5037.4  375.29
  5128.2  377.01  5153.1  379.96  5158.4  377.69  5183.3  379.56  5230.5  381.17
  5243.9  384.47  5262.5  386.03  5293.7  392.16  5329.3  396.26    5348  399.19
  5369.3  403.85  5384.5  404.51  5390.7  406.29  5433.4  411.77  5454.8  415.91
#Mann= 4 ,-1 , 0
  4777.6     .16       0  4838.8     .12       0  4988.1     .07       0
  4994.1     .12       0
Bank Sta=4970.3,5024.5
XS Rating Curve= 0 ,0
Exp/Cntr=0.3,0.1

Type RM Length L Ch R = 1 ,74235   ,356,356,356
XS GIS Cut Line= 3
     3725169.568    10699493.308     3724937.797    10699708.152
     3724699.516     10700119.61
#Sta/Elev= 30
       0  402.83    9.88   402.7   29.64  400.83   88.91  391.55  128.42   386.5
  148.18  384.86  167.94  380.47  177.81  377.14  187.69  376.16  197.57  373.58
  207.45     374  217.33  375.73  246.85  374.99  256.62  375.61  276.16  374.26
   295.7  374.23  334.92   374.5  364.45  375.96  423.51  376.21  443.19  377.48
  453.03  379.35  491.13  384.48  500.54  384.85  547.63  389.63  594.71   395.8
  604.13  396.18  710.69  408.38  720.44   408.5   765.3  414.35  790.67     419
#Mann= 3 ,-1 , 0
       0     .16       0  197.57     .07       0  207.45     .16       0
Bank Sta=167.94,453.03
XS Rating Curve= 0 ,0
Exp/Cntr=0.3,0.1

Type RM Length L Ch R = 1 ,73879   ,506,506,506
BEGIN DESCRIPTION:
BEAVER CREEK 115.0
END DESCRIPTION:
XS GIS Cut Line= 3
      3725099.64      10699360.2      3724899.61     10699310.19
      3724099.58     10699760.21
#Sta/Elev= 30
  4811.6  389.25  4853.2  383.64  4904.4  379.04    4925  374.95  4954.2  374.68
  4976.6  375.26  4994.6  371.42  5025.8  374.07    5144  371.53  5215.1  373.06
  5338.3  371.96    5362  371.65  5398.6  376.31  5407.9  375.77  5411.6  371.38
  5414.3  370.88  5417.6  371.38  5511.1  374.71  5560.5  377.22  5614.1  386.73
  5619.8  385.57  5635.8  390.46  5641.5  389.86  5684.8  397.68  5760.1  415.02
    5775  416.79  5781.7  420.09  5787.5  419.76  5840.6  430.72  5935.7  444.84
#Mann= 7 ,-1 , 0
  4811.6     .16       0  4853.2     .12       0  4954.2     .07       0
  5338.3     .12       0  5411.6     .07       0  5417.6     .12       0
  5840.6     .16       0
Bank Sta=4976.6,5511.1
XS Rating Curve= 0 ,0
Exp/Cntr=0.3,0.1

Type RM Length L Ch R = 1 ,73373   ,401,401,401
BEGIN DESCRIPTION:
BEAVER CREEK 114.0
END DESCRIPTION:
XS GIS Cut Line= 3
      3725099.59     10697860.23      3724599.61     10699060.19
      3724199.64     10699460.16
#Sta/Elev= 30
  3718.7  404.18  3839.4  395.96  3946.2   376.7  4022.5   374.3  4336.2  371.33
  4542.5  372.52  4552.8  366.69  4560.9  372.56  4720.2  371.63    4737  365.35
    4744   370.6  4749.4  368.46  4767.9  371.01  4932.5  371.07  4956.4  377.32
  4980.2  376.42  4986.2  373.08    5004   371.4  5009.4  375.09  5046.9  376.15
  5075.2  372.54  5160.1  368.76  5185.4  364.38  5188.1  363.88  5191.4  364.38
  5216.6   369.3  5301.5   369.4  5372.2  373.89  5428.8  377.92  5584.3  405.06
#Mann= 3 ,-1 , 0
  3718.7     .12       0  5185.4     .07       0  5191.4     .12       0
Bank Sta=5075.2,5372.2
XS Rating Curve= 0 ,0
Exp/Cntr=0.3,0.1

Type RM Length L Ch R = 1 ,72972   ,450,450,450
BEGIN DESCRIPTION:
BEAVER CREEK 113.0
END DESCRIPTION:
XS GIS Cut Line= 3
      3725049.58     10697710.23      3724219.14     10698963.67
       3723849.6     10699110.19
#Sta/Elev= 30
  3548.2  428.15  3672.7   413.2    3743  403.07  3901.6  380.05  3994.9  374.88
  4118.2  371.63  4262.6  373.17  4340.8  370.06  4349.9  366.94  4376.9  370.35
  4449.1  370.26  4464.2   367.9  4479.2   369.8  4500.3  365.21  4507.8  369.95
  4659.7  369.87  4677.7  363.18  4680.5  362.68  4683.7  363.18  4687.7  368.39
  4695.8   369.7  4912.4  366.88  4975.6  368.58  4984.6  364.42  5005.6  363.55
  5011.6  366.73  5046.8  369.14  5134.6  373.79  5341.7  397.62  5449.3  414.11
#Mann= 5 ,-1 , 0
  3548.2     .05       0  3672.7     .07       0    3743     .12       0
  4677.7     .07       0  4683.7     .12       0
Bank Sta=4975.6,5046.8
XS Rating Curve= 0 ,0
Exp/Cntr=0.3,0.1

Type RM Length L Ch R = 1 ,72522   ,508,508,508
BEGIN DESCRIPTION:
BEAVER CREEK 112.0
END DESCRIPTION:
XS GIS Cut Line= 3
       3724899.6     10697610.19      3723999.61     10698610.19
      3723649.58     10698860.21
#Sta/Elev= 30
  3654.9  426.13  3718.8  425.55  3820.6  413.62  3867.5  406.61  3881.7  406.11
  3910.1  401.28  4065.6  382.74  4100.7  383.33  4206.9  374.83  4334.7  370.99
  4469.2  369.35  4554.4  368.86  4561.1  370.21  4582.8  368.43  4915.4  367.41
    4979   368.4  4986.4  364.75  4993.2  366.35  4996.9  361.94  5004.6  361.76
  5007.4  361.26  5010.6  361.76  5013.8  366.22  5037.1  368.76  5064.2  371.94
  5108.4  370.86  5194.4  381.71  5200.6  384.16    5337  402.88  5430.4  424.88
#Mann= 4 ,-1 , 0
  3654.9     .05       0  3820.6     .12       0  5004.6     .07       0
  5010.6     .12       0
Bank Sta=4979,5037.1
XS Rating Curve= 0 ,0
Exp/Cntr=0.3,0.1

Type RM Length L Ch R = 1 ,72014   ,414,414,414
BEGIN DESCRIPTION:
BEAVER CREEK 111.0
END DESCRIPTION:
XS GIS Cut Line= 3
      3724299.63     10697760.17      3723699.61     10698360.19
      3723499.58      10698460.2
#Sta/Elev= 30
  4138.9   402.6  4209.6  391.86  4294.5  383.69  4322.8   378.3  4464.2  371.37
  4492.5  371.14  4506.6  368.57  4591.5  367.21  4633.9  367.81  4690.5  365.78
  4732.9  367.14    4846  366.77  4874.3  365.98  4888.5  363.76  4973.3  367.41
  4983.9  363.01  4990.3  363.01  4998.4  360.74  5001.2  360.24  5004.4  360.74
  5009.8  366.26  5023.8  367.39  5040.6  367.67  5068.5  371.84  5085.3  371.43
  5099.3  375.04  5107.6  381.81    5158  392.28  5197.1  399.29  5211.1  400.68
#Mann= 3 ,-1 , 0
  4138.9     .12       0  4998.4     .07       0  5004.4     .12       0
Bank Sta=4973.3,5023.8
XS Rating Curve= 0 ,0
Exp/Cntr=0.3,0.1

Type RM Length L Ch R = 1 ,71600   ,600,600,600
BEGIN DESCRIPTION:
BEAVER CREEK 110.0
END DESCRIPTION:
XS GIS Cut Line= 2
      3724006.46     10697414.19      3723404.06     10698324.29
#Sta/Elev= 30
  4171.2  407.27  4173.5  405.26  4202.4  403.27  4209.6  401.62  4230.6   401.2
  4270.4  395.32  4346.3   378.4  4369.1  376.42  4382.3  372.77  4411.2   370.5
  4426.2  370.99  4432.2  369.17  4462.3  369.34  4483.4  367.42  4540.5  365.61
  4627.8  364.52  4880.5  365.99  4931.7  364.19  4981.9  366.13  4988.9  362.87
  4991.9   358.6  4994.6   358.1  4997.9   358.6  5003.9  358.68  5009.9  365.45
  5139.3   365.8  5161.7  369.35  5175.4  377.08  5197.7  382.42  5262.6  393.12
#Mann= 4 ,-1 , 0
  4171.2     .05       0  4270.4     .12       0  4991.9     .07       0
  4997.9     .12       0
Bank Sta=4981.9,5009.9
XS Rating Curve= 0 ,0
Exp/Cntr=0.3,0.1

Type RM Length L Ch R = 1 ,71000   ,383,383,383
BEGIN DESCRIPTION:
BEAVER CREEK 109.0
END DESCRIPTION:
XS GIS Cut Line= 3
      3723849.59      10697310.2      3723249.61     10697660.19
      3722649.64     10698210.16
#Sta/Elev= 30
  4314.8  391.75  4384.7  383.45  4430.5   374.4  4461.6  370.36  4541.8  366.47
  4754.7  363.47    4980  364.68  4992.8   356.9  4995.5   356.4  4998.8   356.9
  5006.5  362.91  5016.5   362.4  5023.3  364.41  5136.7  363.36  5150.9  361.86
  5186.1  363.47  5200.2  358.97  5207.6  363.42  5242.8  365.59  5250.2  368.05
  5321.1  372.78    5363   373.1  5433.9  379.01  5497.8  388.73  5582.6  398.42
  5632.5  406.51    5717   415.3  5781.1  424.16  5787.9  423.66  5823.3  429.15
#Mann= 4 ,-1 , 0
  4314.8     .05       0  4384.7     .12       0  4992.8     .07       0
  4998.8     .12       0
Bank Sta=4980,5023.3
XS Rating Curve= 0 ,0
Exp/Cntr=0.3,0.1

Type RM Length L Ch R = 1 ,70617   ,78,78,78
BEGIN DESCRIPTION:
Mapping XS a37a6844
END DESCRIPTION:
XS GIS Cut Line= 6
      3723100.07     10696678.09      3723130.45      10697090.4
      3723061.01     10697428.94      3722922.12     10697875.99
      3722631.32      10697984.5      3722372.75     10698057.76
#Sta/Elev= 30
  4223.8  385.43    4246  388.89    4266  384.22  4316.2   386.2  4356.3   383.3
  4405.9  376.23  4418.9  377.14  4486.7  370.37  4504.5  370.53    4603  369.15
    4627  369.49  4647.2  365.27    4702  364.02  4801.3  363.02  4900.6  363.32
  4986.1  361.91  4999.4  356.78  5002.1  356.28  5005.4  356.78  5015.5  362.93
  5106.6   362.7  5418.5  369.14  5473.2   373.2  5578.5  385.32  5625.6  391.07
    5806  405.73  5834.8  406.36    5913  415.14  5963.3  418.15  6030.9  422.27
#Mann= 12 ,-1 , 0
  4223.8     .12       0  4405.9     .05       0  4504.5     .08       0
    4603     .05       0    4702     .08       0  4801.3      .1       0
  4900.6     .12       0  4999.4     .07       0  5005.4     .12       0
  5106.6     .05       0  5578.5     .12       0  5963.3     .05       0
Bank Sta=4986.1,5015.5
XS Rating Curve= 0 ,0
Exp/Cntr=0.3,0.1

Type RM Length L Ch R = 1 ,70539   ,867,867,867
BEGIN DESCRIPTION:
BEAVER CREEK 108.0
END DESCRIPTION:
XS GIS Cut Line= 6
      3722994.25      10696691.1      3723046.33     10697027.89
      3723004.67     10697371.64      3722921.33     10697694.55
      3722844.94     10697795.25      3722268.94     10697965.29
#Sta/Elev= 30
    4279   388.4  4282.2  389.63  4328.7  382.87  4545.7  369.59  4607.7  366.07
  4630.6  367.76  4717.5   363.8  4743.4  364.71  4773.2  362.19  4783.3  358.36
  4799.4   361.7  4962.8  364.38  4982.2  355.81    4985  355.31  4988.2  355.81
  4995.5  356.67  5003.5  360.96  5026.5  364.16  5247.5  363.03    5428   369.1
  5474.3  369.81  5509.8  374.71  5613.8  383.84  5618.9  386.11  5654.8  386.77
  5666.1   389.4  5848.8  400.11  5951.9   406.8  5988.6  409.47  6027.7  409.12
#Mann= 9 ,-1 , 0
    4279     .05       0  4545.7     .12       0  4743.4     .05       0
  4982.2     .04       0  4988.2     .05       0    5428     .07       0
  5509.8     .05       0  5848.8     .08       0  5951.9     .05       0
Bank Sta=4962.8,5026.5
XS Rating Curve= 0 ,0
Exp/Cntr=0.3,0.1

Type RM Length L Ch R = 1 ,69672   ,601,601,601
BEGIN DESCRIPTION:
BEAVER CREEK 107.0
END DESCRIPTION:
XS GIS Cut Line= 3
       3722749.6     10696510.21      3722649.61     10696910.19
      3721849.61     10697610.19
#Sta/Elev= 30
  4594.6  399.37  4635.8  396.53  4723.3  386.34  4749.2  382.26    4811  368.41
  4831.7  366.14  4914.1  359.81    4976  360.79  4983.7  359.08  4996.6  352.93
  5001.3  352.89  5004.1  352.39  5007.3  352.89  5010.2  352.89    5014  359.42
  5020.7  359.98  5056.7  360.76  5063.4  358.01    5071  361.06  5155.4  359.08
  5226.6   361.3  5410.7   360.9    5779  371.59  5821.7  373.86  5829.3  375.97
    5860  378.16  5963.6  392.37  5999.2  399.83  6005.8  399.34  6069.9  409.03
#Mann= 5 ,-1 , 0
  4594.6     .05       0  4723.3     .12       0  5001.3     .07       0
  5007.3     .12       0    5860     .05       0
Bank Sta=4976,5020.7
XS Rating Curve= 0 ,0
Exp/Cntr=0.3,0.1

Type RM Length L Ch R = 1 ,69071   ,570,570,570
BEGIN DESCRIPTION:
BEAVER CREEK 106.0
END DESCRIPTION:
XS GIS Cut Line= 3
      3722649.65     10696460.17      3722199.61     10696660.19
      3721599.62     10697160.18
#Sta/Elev= 30
  4488.9  393.61  4526.6  390.43  4573.1  383.76  4642.2  375.41  4653.8  372.25
  4775.5  360.64    4861   358.1  4920.5  359.33    4967  357.29  4972.5  358.75
  4984.6  357.23  4988.6  352.33  4995.1  353.74  5006.4  352.17  5009.1  351.67
  5012.4  352.17  5017.2  357.06  5031.5  357.79  5208.5  360.22  5358.2  366.51
  5399.9  370.26  5472.3  382.06  5500.1  388.03  5506.6  387.21  5514.4  390.32
  5541.8  395.24  5599.1  402.89    5642   411.3  5677.2  413.65  5762.4  424.09
#Mann= 5 ,-1 , 0
  4488.9     .05       0  4573.1     .12       0  5006.4     .07       0
  5012.4     .12       0  5472.3     .05       0
Bank Sta=4972.5,5031.5
XS Rating Curve= 0 ,0
Exp/Cntr=0.3,0.1

Type RM Length L Ch R = 1 ,68501   ,467,467,467
BEGIN DESCRIPTION:
BEAVER CREEK 105.0
END DESCRIPTION:
XS GIS Cut Line= 3
      3722649.57      10696060.2      3721849.61     10696310.19
      3721499.63     10696860.16
#Sta/Elev= 30
  4177.9  407.92  4291.5   394.6  4296.8  395.63  4329.3  393.48  4361.7  387.26
    4367  387.99  4531.4  367.79    4624  358.99  4806.5  356.67  4879.3  358.41
  4971.9  358.11  4974.1   358.2  4984.6   357.5  4996.8  351.45  4999.5  350.95
  5002.8  351.45  5013.4  355.84  5038.9  356.98  5044.8  353.13  5051.6  357.36
  5102.4  356.53    5154  359.01  5217.5  359.24  5253.9  361.67  5263.2  360.59
  5305.6  366.16  5377.6  379.84  5457.1  393.42  5466.4  392.77  5667.9  415.89
#Mann= 8 ,-1 , 0
  4177.9     .05       0  4531.4     .16       0    4624     .12       0
  4879.3     .05       0  4971.9     .12       0  4996.8     .07       0
  5002.8     .12       0  5377.6     .05       0
Bank Sta=4974.1,5051.6
XS Rating Curve= 0 ,0
Exp/Cntr=0.3,0.1

Type RM Length L Ch R = 1 ,68034   ,469,469,469
BEGIN DESCRIPTION:
Mapping XS d73e9fa1
END DESCRIPTION:
XS GIS Cut Line= 2
      3722545.73     10695611.23      3721116.39      10696235.7
#Sta/Elev= 30
  4016.3  413.34  4056.2  413.55  4097.5  410.03  4178.6  398.53    4202   397.1
  4248.8  390.09  4254.3  388.04  4371.5  373.51  4400.2  368.26  4415.8  367.63
  4423.6  364.75  4551.5  355.49  4808.7  357.06  4994.2  356.45    4997  351.37
  4999.7  350.87    5003  351.37    5016  352.22  5028.9  355.96  5081.5  355.17
  5203.6  360.84  5244.9  364.23  5256.1  367.19  5297.2  371.43  5350.3  374.96
  5425.1  374.68  5448.5  376.63  5477.4  376.71    5570  386.67  5576.1   386.6
#Mann= 6 ,-1 , 0
  4016.3     .05       0  4371.5     .12       0    4997     .07       0
    5003     .12       0  5350.3     .05       0    5570     .08       0
Bank Sta=4994.2,5028.9
XS Rating Curve= 0 ,0
Exp/Cntr=0.3,0.1

Type RM Length L Ch R = 1 ,67565   ,633,633,633
BEGIN DESCRIPTION:
BEAVER CREEK 104.0
END DESCRIPTION:
XS GIS Cut Line= 3
      3722511.06     10695215.39      3721719.37     10695083.44
      3721261.91     10695956.77
#Sta/Elev= 30
  3627.4  409.05  3659.3  409.25    3687  406.64  3692.1  407.88  3747.9  400.57
  3752.9  401.64  3808.7  395.04  3813.8  396.37  3991.2  379.92  3996.2  380.81
  4024.2  377.37  4070.4   375.3  4095.2  373.58  4234.5  356.52  4295.3     354
  4932.3  354.53  4945.6  352.29  4976.4  353.62  4982.1  351.96  5001.2  351.38
  5003.9  350.88  5007.2  351.38  5070.3  354.38  5191.4  359.94  5256.2  367.36
  5279.7  371.87  5340.3  379.37    5390  380.26  5412.1  383.29  5415.9   386.1
#Mann= 5 ,-1 , 0
  3627.4     .05       0  4070.4     .12       0  5001.2     .07       0
  5007.2     .12       0  5256.2     .05       0
Bank Sta=4932.3,5070.3
XS Rating Curve= 0 ,0
Exp/Cntr=0.3,0.1
