HEC-RAS study BEAVER CREEK.prj: BEAVER CREEK Base Level Engineering

--- BEAVER CREEK.g01 (geometry) --- (continued)

Type RM Length L Ch R = 1 ,66932   ,87,87,87
BEGIN DESCRIPTION:
Mapping XS 115b8afd
END DESCRIPTION:
XS GIS Cut Line= 4
      3722657.02     10694304.43      3721582.41     10694729.76
      3721393.67     10695213.66      3721155.51     10695963.84
#Sta/Elev= 30
  3545.4   410.9  3680.2  394.85  3734.2  384.46  3940.5  384.46  3994.3  389.56
  4088.3  371.66  4147.8  364.67  4201.8  367.61  4226.2  364.08  4309.9  364.32
  4339.6  359.83  4388.3  363.33  4393.7  358.84    4418  363.26  4721.3  357.02
  4755.4  353.81  4851.9  354.84  4873.3  351.47  4888.6  354.05  4945.5  351.26
  4948.2  350.76  4951.5  351.26  5024.7  353.94  5081.5  354.51  5364.4  356.24
  5547.6  359.04  5681.9   366.9  5708.9  365.15  5841.6  378.65  6007.6   385.2
#Mann= 7 ,-1 , 0
  3545.4     .14       0  4721.3     .14       0  4945.5     .07       0
  4951.5     .14       0  5024.7     .14       0  5364.4     .14       0
  5841.6     .05       0
#XS Ineff= 2 , 0
       0 4793.63  361.24 5124.21       0  361.34
Permanent Ineff=
       T       T
Bank Sta=4851.9,5081.5
XS Rating Curve= 0 ,0
Exp/Cntr=0.3,0.1

Type RM Length L Ch R = 1 ,66845   ,591,591,591
BEGIN DESCRIPTION:
BEAVER CREEK 102.0
END DESCRIPTION:
XS GIS Cut Line= 4
      3721851.32     10693888.98      3721504.09     10694659.83
      3721351.31     10695125.11      3721045.74     10695882.09
#Sta/Elev= 30
  3828.8  385.58  3920.8   386.6  3938.4  376.84  3949.1  382.25  3990.2  372.25
  3995.7   379.4  4013.3  369.84  4019.4  375.35  4059.6  365.61  4212.6  360.58
  4230.8  361.11  4336.5  359.12  4476.1  360.35  4547.8  360.23  4763.4  359.45
  4858.1  360.85  4893.7  360.81  4927.8  351.41  4930.5  350.91  4933.8  351.41
    4960  351.51  5061.9  359.13  5074.6  360.07    5372  358.76  5422.8  359.94
  5476.1  362.07  5580.2  367.19  5715.1  374.98  5788.4  379.94  5980.3   402.7
#Mann= 20 ,-1 , 0
  3828.8     .05       0  3949.1     .12       0  4019.4     .08       0
  4212.6     .12       0  4230.8     .05       0  4336.5     .08       0
  4476.1     .12       0  4547.8     .08       0  4763.4     .12       0
  4858.1     .05       0  4927.8     .07       0  4933.8     .05       0
    4960     .08       0  5061.9     .05       0    5372     .08       0
  5422.8     .12       0  5476.1     .05       0  5580.2     .08       0
  5715.1     .05       0  5788.4     .08       0
#XS Ineff= 2 , 0
       0 4861.22  361.67  5109.5       0  361.71
Permanent Ineff=
       T       T
Bank Sta=4893.7,5074.6
XS Rating Curve= 0 ,0
Exp/Cntr=0.3,0.1

Type RM Length L Ch R = 1 ,66254   ,560,560,560
BEGIN DESCRIPTION:
BEAVER CREEK 101.0
END DESCRIPTION:
XS GIS Cut Line= 3
      3721749.62     10693860.17      3720949.61     10694660.19
      3720649.58     10694960.22
#Sta/Elev= 30
    3900  405.15  3928.3  404.37  3984.9  399.16    3999  395.97  4069.7  386.24
  4154.6  377.45  4225.3   364.5  4253.6  361.51  4338.4  357.13  4621.3  352.22
  4805.1  351.92  4960.7  353.46  4974.8  348.99    4989  349.83  5000.1  348.13
  5002.9  347.63  5006.1  348.13  5017.2  348.18  5027.9  351.08  5045.5  349.76
  5073.8  354.38    5088  354.33  5130.4  358.96  5172.8  365.53  5201.1  372.44
  5257.7  379.72    5275  383.23  5328.4  390.27  5416.4  396.71  5455.7  398.57
#Mann= 5 ,-1 , 0
    3900     .12       0  5000.1     .07       0  5006.1     .12       0
    5275     .16       0  5416.4      .1       0
Bank Sta=4960.7,5073.8
XS Rating Curve= 0 ,0
Exp/Cntr=0.3,0.1

Type RM Length L Ch R = 1 ,65694   ,549,549,549
BEGIN DESCRIPTION:
BEAVER CREEK 100.0
END DESCRIPTION:
XS GIS Cut Line= 3
       3721099.6      10693510.2      3720599.61     10694310.19
      3720549.61      10694710.2
#Sta/Elev= 30
  4050.6  404.65  4109.5  400.86  4189.1  390.37  4231.6  388.03  4274.6  381.18
    4320  377.37  4325.9  378.94  4356.6  374.28  4362.5  375.67  4377.8  372.05
  4383.7  373.44  4414.4  370.37  4420.3  372.03  4435.6  368.91  4441.5   371.4
  4478.1  369.62  4535.8  359.09  4630.2  348.25  4645.5  349.57  4663.7  347.37
  4666.5  346.87  4669.7  347.37    4688  349.77    4971  350.69    4991  347.93
  5024.2  350.65  5104.8  351.53  5161.3   359.7  5245.9  371.86  5397.1  383.03
#Mann= 4 ,-1 , 0
  4050.6     .12       0  4663.7     .07       0  4669.7     .12       0
  5161.3     .16       0
Bank Sta=4971,5024.2
XS Rating Curve= 0 ,0
Exp/Cntr=0.3,0.1

Type RM Length L Ch R = 1 ,65145   ,443,443,443
BEGIN DESCRIPTION:
BEAVER CREEK 99.0
END DESCRIPTION:
XS GIS Cut Line= 3
      3720649.61     10693460.19      3720249.61     10694010.19
       3719949.6     10694560.21
#Sta/Elev= 30
  4330.5  394.65  4388.1  388.97  4394.3  385.82  4466.5   377.1    4480  373.65
  4509.4  369.88  4524.1  369.58    4545   365.6  4559.6  364.96  4645.4  353.43
  4660.1  353.62  4666.3  352.03  4716.5  348.32  4760.6  348.71  4828.7  346.58
  4831.4  346.08  4834.7  346.58  4973.9  349.12  4982.4  347.49    4997  347.41
  5024.3  348.99    5106   347.1  5253.1  348.46  5306.7  353.65    5342   359.9
  5409.3  369.65  5511.8  388.94  5585.3  398.88  5591.5  401.04  5637.1  406.15
#Mann= 4 ,-1 , 0
  4330.5     .12       0  4828.7     .07       0  4834.7     .12       0
    5342     .16       0
Bank Sta=4973.9,5024.3
XS Rating Curve= 0 ,0
Exp/Cntr=0.3,0.1

Type RM Length L Ch R = 1 ,64702   ,989,989,989
BEGIN DESCRIPTION:
Mapping XS 8c4eb2a6
END DESCRIPTION:
XS GIS Cut Line= 2
      3720396.79     10693227.46      3719547.78     10694409.82
#Sta/Elev= 30
  4090.8  385.79  4112.2  384.15  4126.9  385.86  4162.5  385.63  4168.6  384.02
  4212.8  382.91    4219  380.85  4248.4  380.55  4254.6  378.59  4263.2  379.64
  4269.3   377.4  4298.8  375.44  4304.9  372.14  4328.1  368.41  4355.3  359.84
  4405.6  350.67  4414.2  348.68  4476.8  346.48  4645.7   345.6  4648.5   345.1
  4651.7   345.6  4950.8  348.28  5036.7  347.18  5101.8  350.56  5244.2   359.4
  5300.7  370.24  5365.8  378.39  5481.2  396.84  5531.5  406.69  5546.4  406.53
#Mann= 3 ,-1 , 0
  4090.8     .12       0  4645.7     .07       0  4651.7     .12       0
Bank Sta=4405.6,5101.8
XS Rating Curve= 0 ,0
Exp/Cntr=0.3,0.1

Type RM Length L Ch R = 1 ,63713   ,406,406,406
BEGIN DESCRIPTION:
Mapping XS 1c63e403
END DESCRIPTION:
XS GIS Cut Line= 2
      3719827.33     10692894.15      3719003.63     10694203.39
#Sta/Elev= 30
    4576  394.69  4630.4     397  4679.3  393.06  4788.8  372.65  4840.6  359.38
  4854.9  358.07  4861.8   355.4    4883  353.87  4904.2  348.27  4919.5  346.67
  4925.8  344.77  4958.9  343.82  4961.6  343.32  4964.9  343.82  5055.5  344.29
  5114.8     345  5124.2  344.23  5505.9  344.98  5688.4  351.96  5746.1   351.7
  5870.9  361.27  5906.4  365.29  5919.2  368.87  6013.4  381.75  6022.8  381.25
  6028.7  382.96  6059.3  384.33  6065.2  386.09    6117  386.37  6122.8  388.27
#Mann= 5 ,-1 , 0
    4576     .12       0  4958.9     .07       0  4964.9     .12       0
  5055.5     .16       0  5124.2     .12       0
Bank Sta=4919.5,5114.8
XS Rating Curve= 0 ,0
Exp/Cntr=0.3,0.1

Type RM Length L Ch R = 1 ,63307   ,578,578,578
BEGIN DESCRIPTION:
BEAVER CREEK 96.0
END DESCRIPTION:
XS GIS Cut Line= 3
      3719499.63     10692760.15      3719299.61     10693110.19
      3718549.64     10693910.16
#Sta/Elev= 30
  4550.4  396.15  4601.6  393.34  4644.7  387.21  4682.2  379.99  4688.7   376.7
  4725.4  370.46  4741.2  364.33  4769.3  357.98  4827.6  346.55  4834.6  346.02
  4849.9  343.17  5034.7  343.16    5071   342.6  5073.7   342.1    5077   342.6
  5349.9  344.33  5399.3  343.22  5413.4  344.78  5625.4  343.38  5696.3  346.94
  5731.9   350.1  5738.8  352.18  5746.1  351.69  5809.6  362.07  5837.9  363.88
  5915.6  375.49  5922.9  375.14  5929.7  377.27  5979.6  381.76  6050.1  390.98
#Mann= 5 ,-1 , 0
  4550.4     .12       0  4834.6     .16       0  5034.7     .12       0
    5071     .07       0    5077     .12       0
Bank Sta=4827.6,5413.4
XS Rating Curve= 0 ,0
Exp/Cntr=0.3,0.1

Type RM Length L Ch R = 1 ,62729   ,468,468,468
BEGIN DESCRIPTION:
BEAVER CREEK 95.0
END DESCRIPTION:
XS GIS Cut Line= 3
       3719049.6      10692410.2      3718899.61     10692810.19
      3718349.63     10693560.16
#Sta/Elev= 30
  4571.5  391.37  4611.5   389.2  4635.6  385.75  4678.3  375.67  4732.6  366.15
  4752.2  361.02  4787.8  356.27  4812.7  350.39  4849.2  344.87  4881.2  342.33
  5023.9  340.54  5026.6  340.04  5029.9  340.54  5391.7  341.61  5434.4  342.95
  5442.9  344.74  5449.1  347.35  5457.5     347  5478.4  350.99  5507.1  354.45
  5513.9  353.89  5520.1  355.76  5620.4  367.03  5664.4  374.84    5679  376.08
  5693.6   379.4  5850.4  397.23  5856.6  399.38  5879.1  402.05  5928.7   406.9
#Mann= 5 ,-1 , 0
  4571.5     .12       0  5023.9     .07       0  5029.9     .12       0
  5391.7     .16       0  5693.6     .12       0
Bank Sta=4849.2,5442.9
XS Rating Curve= 0 ,0
Exp/Cntr=0.3,0.1

Type RM Length L Ch R = 1 ,62261   ,508,508,508
BEGIN DESCRIPTION:
BEAVER CREEK 94.0
END DESCRIPTION:
XS GIS Cut Line= 2
      3718920.69      10692009.5      3718244.11     10693268.98
#Sta/Elev= 30
  4416.4  390.02  4491.8  388.94  4497.5  386.72  4551.9  381.72  4595.7  373.78
  4632.9  369.79  4644.1  366.63  4741.5  372.46  4780.4  373.23  4825.5  368.77
    4853  364.15  4859.9  361.14  4913.1  349.48  4950.7  343.96  4984.8  339.17
  5027.2  339.14  5029.9  338.64  5033.2  339.14  5324.3  341.55  5416.1  341.17
  5450.2  344.19  5528.8  354.91    5539  355.95  5569.9   362.4  5613.7  367.89
  5620.4  370.49  5679.4  376.96  5695.7  380.56  5739.5  381.47  5846.1  390.34
#Mann= 8 ,-1 , 0
  4416.4     .12       0  4644.1     .16       0  4741.5     .12       0
  5027.2     .07       0  5033.2     .12       0  5324.3     .16       0
  5528.8     .12       0    5539     .16       0
Bank Sta=4950.7,5450.2
XS Rating Curve= 0 ,0
Exp/Cntr=0.3,0.1

Type RM Length L Ch R = 1 ,61753   ,669,669,669
BEGIN DESCRIPTION:
BEAVER CREEK 93.0
END DESCRIPTION:
XS GIS Cut Line= 2
      3718405.08     10691894.89      3717951.95     10692973.03
#Sta/Elev= 30
    4442  391.41    4472  390.73  4512.8  386.82  4519.5  384.25  4548.6   379.6
  4556.2  376.35  4572.4  374.28  4577.9  371.53  4596.1  367.61  4625.3  362.67
  4649.1  356.01  4696.6  347.93  4740.6  343.49  4784.1  339.03  4889.5  337.58
  4892.2  337.08  4895.5  337.58  4963.6  338.46  5047.4  338.55  5250.5  340.46
    5283  343.22  5358.9  351.99  5373.8  356.05  5397.5  358.28  5426.7  364.99
  5479.6  373.05  5574.6  382.25  5580.1  384.57  5603.8  384.24  5611.5  386.13
#Mann= 5 ,-1 , 0
    4442     .12       0  4889.5     .07       0  4895.5     .12       0
  4963.6     .16       0  5047.4     .12       0
Bank Sta=4740.6,5283
XS Rating Curve= 0 ,0
Exp/Cntr=0.3,0.1

Type RM Length L Ch R = 1 ,61084   ,307,307,307
BEGIN DESCRIPTION:
Mapping XS c5f4612c
END DESCRIPTION:
XS GIS Cut Line= 3
      3717906.32      10691672.8      3717754.41     10692488.77
      3717776.05     10693177.04
#Sta/Elev= 30
  4591.4  389.93  4629.4  387.62  4670.1   382.1  4771.8   360.8  4818.4  353.76
  4823.5  351.58  4904.1  341.02  4944.8  336.98  5074.2  336.98  5130.3  337.02
  5165.5  336.58  5168.3  336.08  5171.5  336.58  5300.8  339.47  5313.5  338.34
    5372  341.39  5409.5  345.05  5467.7  351.42  5602.9  370.73  5662.9  377.42
  5702.9  379.15    5813  377.03  5860.5  378.72    5913  382.95  5958.8  383.27
  6043.1  381.88  6061.1  380.05  6066.1  383.83  6093.1  380.32    6110   382.5
#Mann= 9 ,-1 , 0
  4591.4     .12       0  5074.2     .16       0  5130.3     .12       0
  5165.5     .07       0  5171.5     .12       0  5409.5     .16       0
  5467.7     .12       0  5860.5     .16       0  5958.8     .05       0
Bank Sta=4904.1,5372
XS Rating Curve= 0 ,0
Exp/Cntr=0.3,0.1

Type RM Length L Ch R = 1 ,60777   ,482,482,482
BEGIN DESCRIPTION:
Mapping XS 34c8e4e5
END DESCRIPTION:
XS GIS Cut Line= 3
      3717867.25     10691568.65      3717107.71     10692514.82
      3717129.41     10693144.13
#Sta/Elev= 30
  4536.3  389.16    4621  385.58  4678.6  385.93  4728.2  382.75    4877  361.08
  4905.8  352.89  4920.2  345.52  4934.6  340.88  4948.6  339.14  4973.3  336.28
    4976  335.78  4979.3  336.28  5453.1  337.01  5574.7  339.56  5581.1  338.96
  5589.1   342.2  5595.5  340.92  5609.9  345.49  5666.7  354.14  5717.1  365.58
  5749.6  369.31    5775  375.11    5835  381.19  5915.1  382.85  5985.1  380.89
  6165.2  394.75  6215.3   394.1  6255.3  390.15  6325.3  395.02  6379.3  393.05
#Mann= 3 ,-1 , 0
  4536.3     .12       0  4973.3     .07       0  4979.3     .12       0
Bank Sta=4948.6,5574.7
XS Rating Curve= 0 ,0
Exp/Cntr=0.3,0.1

Type RM Length L Ch R = 1 ,60295   ,463,463,463
BEGIN DESCRIPTION:
Mapping XS 57a0bd67
END DESCRIPTION:
XS GIS Cut Line= 4
       3717832.5      10691455.8      3717237.91      10691694.5
      3716777.84     10692623.32      3716708.41     10692944.48
#Sta/Elev= 30
  4234.4  387.04  4302.2  380.37    4340  373.29    4418  362.81  4442.2  361.12
  4447.6  362.53    4496  356.02  4501.3  356.85  4549.7  349.55  4555.1  350.46
  4571.6  346.27    4647  335.34  4968.9  334.49  4988.3  333.67  4991.1  333.17
  4994.3  333.67  5041.8  335.26  5062.6  335.12  5233.7  336.21  5428.6  337.13
  5492.6   345.1  5585.5   355.9  5602.4  359.94  5675.2  371.37  5781.8  382.62
  5918.5  382.59  6067.9  380.24  6073.1  378.47  6133.5     377  6240.2  378.95
#Mann= 7 ,-1 , 0
  4234.4     .12       0  4988.3     .07       0  4994.3     .12       0
  5062.6     .16       0  5233.7     .12       0  5492.6     .16       0
  5918.5     .12       0
Bank Sta=4968.9,5041.8
XS Rating Curve= 0 ,0
Exp/Cntr=0.3,0.1

Type RM Length L Ch R = 1 ,59832   ,451,451,451
BEGIN DESCRIPTION:
BEAVER CREEK 90.0
END DESCRIPTION:
XS GIS Cut Line= 3
      3717749.59     10691310.19      3716949.61     10691460.19
      3716349.63     10691860.17
#Sta/Elev= 30
  4200.3  382.66  4279.1  371.53  4342.7  357.14  4383.4  351.22  4389.3  349.38
  4434.3  343.41  4485.2   338.6  4515.7  336.86  4627.6  338.55  4688.6   337.1
    4709  337.74  4861.6  335.74  4930.3  332.91  4982.8   333.4  4990.9  332.57
  4993.6  332.07  4996.9  332.57  5063.8  334.03  5086.3  332.91  5289.1  335.13
  5325.2  334.59  5346.2  336.16  5410.8  346.42  5418.3  348.81  5446.9  352.17
  5541.5  359.29  5568.6  363.26  5591.1  364.74  5627.2  369.71  5735.3  380.74
#Mann= 3 ,-1 , 0
  4200.3     .12       0  4990.9     .07       0  4996.9     .12       0
Bank Sta=4861.6,5346.2
XS Rating Curve= 0 ,0
Exp/Cntr=0.3,0.1

Type RM Length L Ch R = 1 ,59381   ,724,724,724
BEGIN DESCRIPTION:
BEAVER CREEK 89.0
END DESCRIPTION:
XS GIS Cut Line= 2
      3717321.16     10690558.68      3716135.05      10691765.6
#Sta/Elev= 30
  4114.8  385.92  4166.5  382.71  4215.9  373.13  4272.5  369.23  4322.1  359.79
  4329.1  357.24  4343.2  355.74  4392.8  344.25  4442.2  337.44  4512.9  332.58
  4795.8  332.22  4821.1  330.93  4823.8  330.43  4827.1  330.93  4831.2  332.41
    4909  332.92  4972.5  333.08  5000.8  331.09  5198.8  334.56  5269.6   333.6
  5326.1  337.75  5396.9  344.63    5411  344.61  5418.1  346.35  5545.4   355.5
  5623.2  365.47  5658.6  367.05  5722.2  374.08  5764.6  375.67    5807  380.59
#Mann= 3 ,-1 , 0
  4114.8     .12       0  4821.1     .07       0  4827.1     .12       0
Bank Sta=4442.2,5326.1
XS Rating Curve= 0 ,0
Exp/Cntr=0.3,0.1

Type RM Length L Ch R = 1 ,58657   ,511,511,511
BEGIN DESCRIPTION:
BEAVER CREEK 88.0
END DESCRIPTION:
XS GIS Cut Line= 3
      3716749.59     10690260.22      3716499.61     10690660.19
      3715749.58     10691460.22
#Sta/Elev= 30
  4530.3  367.26  4595.7  360.92  4601.6  358.99    4611  359.72  4624.6  357.32
  4647.6  355.62  4727.2  343.49  4806.3  332.83  4847.1  332.49    4960  331.14
  4973.1  331.59  4988.4  330.87    4996  328.79  4998.8  328.29    5002  328.79
  5019.8  330.52  5037.4  331.08  5103.7  330.73    5163  330.49  5376.9  332.92
  5433.5  331.81  5468.7  332.84  5504.3  331.54  5610.3  331.86  5659.9  333.26
  5872.2  346.72  5886.3  349.03  5949.8  354.19    6028  365.64  6098.6   372.8
#Mann= 10 ,-1 , 0
  4530.3     .12       0  4727.2     .16       0  4806.3     .12       0
  4847.1     .16       0    4960     .07       0    4996     .07       0
    5002     .07       0  5019.8     .12       0  5103.7     .05       0
    5163     .12       0
Bank Sta=4973.1,5037.4
XS Rating Curve= 0 ,0
Exp/Cntr=0.3,0.1

Type RM Length L Ch R = 1 ,58146   ,546,546,546
BEGIN DESCRIPTION:
Mapping XS 1fe27e14
END DESCRIPTION:
XS GIS Cut Line= 3
      3716741.37     10689864.66      3715803.89     10690763.08
      3715457.16     10691265.84
#Sta/Elev= 30
  4007.4  364.14  4019.7  363.75  4026.6  361.56    4048  362.16  4069.1  359.29
  4090.5  360.69  4139.8   357.1  4161.2  358.57  4168.1  356.46  4192.6  355.08
    4260  347.23  4281.3  347.07  4380.4  337.86  4570.2  333.51  4792.4  330.95
  4854.3  331.84  4988.6   330.1  5006.7  327.32  5009.5  326.82  5012.7  327.32
  5016.9  329.83  5060.8  329.44  5231.5  331.51  5372.1  334.23  5515.5   356.3
  5581.1  357.19  5673.7  350.99  5703.2  352.09  5766.3  356.94  5916.6  373.76
#Mann= 8 ,-1 , 0
  4007.4     .16       0  4192.6     .12       0  4570.2     .16       0
  4792.4     .12       0  5006.7     .07       0  5012.7     .12       0
  5060.8     .16       0  5231.5     .12       0
Bank Sta=4988.6,5016.9
XS Rating Curve= 0 ,0
Exp/Cntr=0.3,0.1

Type RM Length L Ch R = 1 ,57600   ,362,362,362
BEGIN DESCRIPTION:
BEAVER CREEK 86.0
END DESCRIPTION:
XS GIS Cut Line= 3
      3715612.91     10689400.23       3715623.6     10690499.14
      3715239.67      10691275.2
#Sta/Elev= 30
  4062.8  370.65  4202.8  361.74  4271.7  349.16  4322.8  338.39  4352.8  334.44
  4682.8  333.36  4872.8  333.99  4892.8  335.35  4933.5  333.99  4962.8  333.72
  4982.8  331.16  4999.8  326.54  5002.6  326.04  5005.8  326.54  5022.8  332.67
  5062.1  333.29  5072.8  331.46  5092.8  332.36  5102.8  330.45  5122.8  333.35
  5352.6  337.26  5612.7  338.38  5674.4  343.23  5876.3  365.37  5881.8  363.62
  5898.7  366.61  5904.3  365.46  5921.1  367.26  5999.7  364.43  6027.6  365.99
#Mann= 6 ,-1 , 0
  4062.8     .16       0  4271.7     .12       0  4933.5     .16       0
  4999.8     .07       0  5005.8     .16       0  5062.1     .12       0
Bank Sta=4962.8,5022.8
XS Rating Curve= 0 ,0
Exp/Cntr=0.3,0.1

Type RM Length L Ch R = 1 ,57238   ,262,262,262
BEGIN DESCRIPTION:
Mapping XS d9579b68
END DESCRIPTION:
XS GIS Cut Line= 4
      3715508.75     10689426.24      3715326.46     10690289.99
      3715230.97     10690619.85      3714944.57     10691049.46
#Sta/Elev= 30
    4026  372.52  4090.4  363.84  4095.5  365.24  4140.1  357.04  4145.2  358.63
  4189.9  352.27    4194  353.84  4239.7  345.33  4244.8  346.63  4295.8  337.64
  4346.9  332.84  4857.9  331.36  4981.9  333.34  4987.2   325.2  4989.4  324.54
  4992.2  324.04  4995.4  324.54  5054.4  332.88  5137.4  344.33  5243.2  363.02
    5395   372.8  5426.4   372.9  5477.5  366.75  5570.6  369.25  5621.7  364.37
  5642.7  366.91  5672.8  364.66  5678.8  366.82  5693.8  364.14  5768.5  366.85
#Mann= 6 ,-1 , 0
    4026     .16       0    4194     .12       0  4989.4     .07       0
  4995.4     .12       0  5137.4     .05       0    5395     .12       0
Bank Sta=4981.9,5054.4
XS Rating Curve= 0 ,0
Exp/Cntr=0.3,0.1

Type RM Length L Ch R = 1 ,56976   ,503,503,503
BEGIN DESCRIPTION:
BEAVER CREEK 85.0
END DESCRIPTION:
XS GIS Cut Line= 3
      3715349.61     10689510.18      3715049.61     10690310.19
      3715049.61     10690710.18
#Sta/Elev= 30
  4144.1  371.33  4181.9  367.14  4239.3  359.92  4244.7  357.06  4261.6  352.72
  4274.9  351.34  4282.9  348.17  4299.9  344.78  4410.2  331.52  4616.7  330.16
  4806.3  332.21  4867.7  330.83  4891.7  331.95  4903.3  330.26  4922.9  331.79
  4977.1  330.95  4988.7  326.69  4992.8  322.57  4995.6  322.07  4998.8  322.57
    5001  322.57  5008.5   329.4  5018.5  331.32  5038.5  330.91  5138.5  341.69
  5162.9  346.67  5218.5  356.58  5268.5  361.02  5358.5  374.62  5398.5  378.12
#Mann= 5 ,-1 , 0
  4144.1     .16       0  4181.9     .12       0  4992.8     .07       0
  4998.8     .12       0  5162.9     .05       0
Bank Sta=4977.1,5018.5
XS Rating Curve= 0 ,0
Exp/Cntr=0.3,0.1

Type RM Length L Ch R = 1 ,56473   ,492,492,492
BEGIN DESCRIPTION:
BEAVER CREEK 84.0
END DESCRIPTION:
XS GIS Cut Line= 3
      3715349.61     10689410.19      3714649.61     10690160.19
      3714699.61     10690610.21
#Sta/Elev= 30
  3966.1  376.82  4001.5  376.33  4095.7  370.15  4171.3  360.06  4192.5  354.41
  4220.9  350.67    4426  329.89  4666.4  328.85  4822.2  331.11  4836.4  328.46
  4878.9  330.15  4885.8  327.61  4907.3  330.58  4921.4  330.68  4935.6  327.67
  4949.8  330.15  4970.8  329.49  4984.9  329.11  4988.6   323.6  4999.1  322.07
  5001.8  321.57  5005.1  322.07  5022.2  327.69  5032.3  328.62  5183.2  330.28
  5223.4  333.11  5289.2     342  5338.7  350.03  5414.6  363.12  5444.8  365.92
#Mann= 6 ,-1 , 0
  3966.1     .16       0  4095.7     .12       0  4999.1     .07       0
  5005.1     .12       0  5289.2     .16       0  5338.7     .05       0
Bank Sta=4970.8,5032.3
XS Rating Curve= 0 ,0
Exp/Cntr=0.3,0.1

Type RM Length L Ch R = 1 ,55981   ,684,684,684
BEGIN DESCRIPTION:
BEAVER CREEK 83.0
END DESCRIPTION:
XS GIS Cut Line= 2
       3714315.3     10689001.71      3714185.15      10690385.7
#Sta/Elev= 30
  3967.2  373.64  4005.8  369.12  4025.9  360.07    4036   358.3    4046  352.47
  4056.1   349.8  4081.3   338.7  4116.3  334.48  4143.9  334.57  4220.7  332.84
  4293.6  330.19  4357.4   330.6  4457.9  326.95  4555.8  326.16  4826.7  326.72
    4950  328.74    4960  328.33  4987.2  320.07  4989.9  319.57  4993.2  320.07
  5000.2  320.37  5020.3  328.31  5030.3  329.23  5080.6  328.65  5147.7  339.25
  5152.7  338.29  5160.9  341.05  5241.3  354.44  5311.5  361.86  5357.3  364.59
#Mann= 8 ,-1 , 0
  3967.2     .12       0  4143.9     .16       0  4220.7     .12       0
  4457.9     .16       0  4555.8     .12       0  4987.2     .07       0
  4993.2     .12       0  5311.5     .16       0
Bank Sta=4950,5030.3
XS Rating Curve= 0 ,0
Exp/Cntr=0.3,0.1

Type RM Length L Ch R = 1 ,55297   ,120,120,120
BEGIN DESCRIPTION:
BEAVER CREEK 82.0
END DESCRIPTION:
XS GIS Cut Line= 6
      3714193.78     10688784.65      3714085.27     10689223.03
      3713998.47       10689414.      3713911.66     10689557.23
      3713616.52     10689787.26       3713581.8     10690494.71
#Sta/Elev= 30
  3717.3  363.37  3752.1   361.3  3759.2   356.1  3774.5   357.7  3793.5  355.87
  3798.7  351.36  3846.6  348.06  4000.6  345.97  4102.4  339.97  4210.8  336.73
  4418.3  327.58  4451.6  327.28  4530.3  325.69  4610.5  324.52  4694.4  324.55
    4735  324.15  4836.4  323.75  4975.1  327.01  4985.3  319.79  4995.1  319.07
  5000.2  321.96  5002.5  318.68  5005.2  318.18  5008.5  318.68  5015.6     319
  5025.7  326.98  5175.2  325.72  5237.1  327.49  5384.4  333.71  5631.1   371.6
#Mann= 16 ,-1 , 0
  3717.3     .16       0  3759.2     .05       0  4102.4     .16       0
  4210.8     .05       0  4418.3     .12       0  4451.6     .05       0
  4530.3     .16       0  4610.5     .08       0  4694.4     .16       0
    4735     .05       0  4836.4     .12       0  5002.5     .07       0
  5008.5     .12       0  5175.2     .05       0  5237.1     .12       0
  5384.4     .16       0
Bank Sta=4975.1,5025.7
XS Rating Curve= 0 ,0
Exp/Cntr=0.3,0.1

Type RM Length L Ch R = 1 ,55177   ,876,876,876
BEGIN DESCRIPTION:
BEAVER CREEK 81.0
END DESCRIPTION:
XS GIS Cut Line= 6
      3714115.66     10688693.47      3713981.11     10689227.37
      3713863.92       10689414.      3713564.44     10689626.67
      3713494.99     10689717.82      3713403.85      10690512.1
#Sta/Elev= 30
  3593.3  359.69  3719.6   357.9  3806.9  362.51  3868.6  358.95  3919.9  355.33
    3925  358.19  3978.1  350.96    4162  344.65  4172.2  344.47  4306.6  341.45
  4343.1  336.92  4363.9  338.63  4407.5  339.03  4414.1  336.38  4442.6  338.71
  4499.1  335.02  4551.3  331.72  4624.7  327.98  4735.2  325.92  4970.8   325.8
  4980.8  324.01  4987.8  317.85  4990.6  317.35  4993.8  317.85  5000.8  317.99
  5010.8  327.01  5333.4  333.85  5422.8  343.26  5541.8  360.34  5648.2  371.01
#Mann= 15 ,-1 , 0
  3593.3     .05       0  3868.6     .12       0  3978.1     .05       0
    4162     .12       0  4172.2     .05       0  4363.9      .1       0
  4407.5     .05       0  4499.1     .16       0  4551.3     .05       0
  4624.7      .1       0  4735.2     .05       0  4987.8     .04       0
  4993.8     .05       0  5422.8     .12       0  5541.8     .05       0
Bank Sta=4970.8,5010.8
XS Rating Curve= 0 ,0
Exp/Cntr=0.3,0.1

Type RM Length L Ch R = 1 ,54301   ,514,514,514
BEGIN DESCRIPTION:
BEAVER CREEK 80.0
END DESCRIPTION:
XS GIS Cut Line= 3
      3713049.63     10689310.16      3712749.61     10689610.19
      3712899.62     10690360.24
#Sta/Elev= 30
  4550.5  369.62  4607.1  365.26  4677.8   356.6    4692  353.27  4706.1  351.51
  4720.2  347.23  4762.7  339.88  4776.8  338.92  4805.1   334.7  4918.2  325.94
  4977.3  324.47    4985  316.77  4992.2  314.26  4994.9  313.76  4998.2  314.26
  5005.4  314.48  5015.6  318.35  5025.8  324.29  5250.1  322.82  5260.3  323.66
  5301.1  321.75  5321.5  323.56  5382.7  323.62  5413.3  327.72  5525.5  338.35
  5596.9  350.87  5658.1  359.02  5668.3  359.03  5723.8  364.48  5739.7  365.43
#Mann= 4 ,-1 , 0
  4550.5     .12       0  4992.2     .07       0  4998.2     .12       0
  5723.8     .05       0
Bank Sta=4977.3,5025.8
XS Rating Curve= 0 ,0
Exp/Cntr=0.3,0.1

Type RM Length L Ch R = 1 ,53787   ,276,276,276
BEGIN DESCRIPTION:
BEAVER CREEK 79.0
END DESCRIPTION:
XS GIS Cut Line= 3
      3712649.61     10688910.19      3712349.61     10689360.19
       3712649.6     10690160.16
#Sta/Elev= 30
  4479.2  390.33  4537.8  382.93  4551.3  380.01  4558.8  376.52  4636.9   363.1
    4682  361.87    4688  359.42  4718.1  358.99  4724.1  355.39  4754.1  353.07
  4847.3  337.06    4984  322.76  4991.5  313.44  4993.9  313.13  4994.5  313.05
  4997.3  312.55  5000.5  313.05  5006.5  315.13    5017  322.03  5046.9  321.29
    5231  321.35  5266.6  323.03  5400.3  321.47  5405.8  321.47  5578.1  322.36
    5597  321.03  5633.2  321.85  5688.4  329.69  5718.7  330.44  5874.4  344.02
#Mann= 8 ,-1 , 0
  4479.2     .12       0  4993.9     .16       0  4994.5     .07       0
  5000.5     .16       0  5046.9     .07       0  5400.3     .12       0
  5405.8     .07       0    5597     .12       0
Bank Sta=4984,5017
XS Rating Curve= 0 ,0
Exp/Cntr=0.3,0.1

Type RM Length L Ch R = 1 ,53511   ,502,502,502
BEGIN DESCRIPTION:
Mapping XS c2429761
END DESCRIPTION:
XS GIS Cut Line= 3
      3712370.59     10688418.26      3712110.17     10689069.34
      3712058.12     10690526.48
#Sta/Elev= 30
  4066.4  359.99  4107.8  358.83  4114.2  356.63    4132  357.46  4208.5   351.2
  4239.7  345.13  4364.3  334.85  4391.6  335.57  4445.4  331.04  4484.8  331.08
  4514.4   328.6  4538.6   330.5    4544  328.67  4616.7  328.89  4765.4  320.89
  4968.6  320.37  4978.6  319.92  4995.6   312.1  4998.4   311.6  5001.6   312.1
  5008.6  319.46  5018.6  320.32  5118.7  319.76  5138.7  321.81  5408.9   318.2
  5503.9  318.92  5530.9  318.83  5679.1  319.03  6044.2  331.18  6225.7  353.95
#Mann= 7 ,-1 , 0
  4066.4     .12       0  4114.2     .16       0  4364.3     .12       0
  4995.6     .07       0  5001.6     .12       0  5503.9     .07       0
  5530.9     .12       0
Bank Sta=4968.6,5018.6
XS Rating Curve= 0 ,0
Exp/Cntr=0.3,0.1

Type RM Length L Ch R = 1 ,53009   ,407,407,407
BEGIN DESCRIPTION:
Mapping XS 9b56d19b
END DESCRIPTION:
XS GIS Cut Line= 2
       3711628.4     10688535.52      3711719.54     10690410.51
#Sta/Elev= 30
  4094.2  336.49  4131.5  334.86    4179  333.95    4199   332.3  4524.4  325.23
  4739.6  320.63  4979.9  318.13  5006.9  311.24  5009.7  310.74  5012.9  311.24
    5020  311.38    5030  317.53    5040  318.89    5090  319.13  5110.1  316.77
  5130.1  318.48  5248.6  317.08  5360.4  317.99  5380.4  316.64  5416.3  316.79
  5470.5  317.72  5522.8  317.01  5610.7  316.68  5630.7   318.3  5664.8  318.07
  5790.9  330.36  5820.9  331.67    5861  335.89  5872.9     336  5971.4  344.32
#Mann= 7 ,-1 , 0
  4094.2     .16       0  4131.5     .05       0  4524.4     .12       0
  5006.9     .07       0  5012.9     .12       0  5416.3     .07       0
  5522.8     .12       0
Bank Sta=4979.9,5040
XS Rating Curve= 0 ,0
Exp/Cntr=0.3,0.1

Type RM Length L Ch R = 1 ,52602   ,527,527,527
BEGIN DESCRIPTION:
BEAVER CREEK 77.0
END DESCRIPTION:
XS GIS Cut Line= 3
      3710699.59     10688710.17      3711299.61     10689510.19
       3711199.6     10690160.22
#Sta/Elev= 30
  3965.9  373.12  4029.5  365.87  4123.2  347.02  4158.6   344.1  4187.8  339.37
  4202.4  339.77  4237.8  334.73  4287.8  330.97  4358.6  330.63  4429.5  325.42
  4458.6  325.14  4502.4   320.3  4608.6  317.07  4787.8  315.45    4976  317.67
  4986.2  317.03    4995  311.23  5000.1  312.87  5003.4  310.69  5006.1  310.19
  5009.4  310.69  5026.6  317.13  5117.7     317  5131.6  315.57  5158.2  316.97
  5168.3  313.12    5229  318.04  5380.7  334.48    5463  345.07  5623.6  357.91
#Mann= 3 ,-1 , 0
  3965.9     .12       0  5003.4     .07       0  5009.4     .12       0
Bank Sta=4976,5026.6
XS Rating Curve= 0 ,0
Exp/Cntr=0.3,0.1

Type RM Length L Ch R = 1 ,52075   ,334,334,334
BEGIN DESCRIPTION:
BEAVER CREEK 76.0
END DESCRIPTION:
XS GIS Cut Line= 3
      3710599.62     10688710.21      3710849.61     10689410.19
      3710899.61     10690060.18
#Sta/Elev= 30
  4227.9  383.59  4323.4  375.34  4330.4  373.49  4355.3  371.06  4376.5  366.09
  4391.9  364.18  4408.4  359.21  4448.2  353.07  4453.5   350.1  4472.1  346.33
  4484.3  341.93  4515.1  336.63  4695.1  319.04  4758.8  314.84  4807.1   313.7
  4981.2  316.35  4988.2  309.92    4991  309.42  4994.2  309.92  5001.3  310.54
  5011.3  315.49  5021.3  316.18  5091.5  315.85  5161.7  322.86    5262  328.25
  5412.5  338.19  5482.7  344.53  5521.8  346.26  5552.9  349.75  5623.1  354.62
#Mann= 4 ,-1 , 0
  4227.9     .12       0  4988.2     .07       0  4994.2     .12       0
  5521.8     .05       0
Bank Sta=4981.2,5021.3
XS Rating Curve= 0 ,0
Exp/Cntr=0.3,0.1

Type RM Length L Ch R = 1 ,51741   ,728,728,728
BEGIN DESCRIPTION:
BEAVER CREEK 75.0
END DESCRIPTION:
XS GIS Cut Line= 2
      3710419.47     10688953.91      3710697.24     10690073.68
#Sta/Elev= 30
  4466.4  371.08    4488   367.7  4493.5  363.34  4529.4  356.71  4534.7  353.56
  4570.8  343.06  4586.2   341.6  4596.5  338.84  4606.8  338.07  4612.2  335.66
  4627.4  334.33  4658.7  328.56  4730.4  320.95  4761.4  316.03    4819  312.66
  4984.5  315.06  4989.7  311.34  4995.3  309.46  4998.1  308.96  5001.3  309.46
  5008.6  313.48  5018.9  315.11  5101.4  314.03  5132.3  317.24  5255.9  321.51
  5356.9  329.44  5369.2  329.16  5522.4  337.29  5616.8  345.71  5620.1  345.71
#Mann= 4 ,-1 , 0
  4466.4     .12       0  4995.3     .07       0  5001.3     .12       0
  5616.8     .05       0
Bank Sta=4984.5,5018.9
XS Rating Curve= 0 ,0
Exp/Cntr=0.3,0.1

Type RM Length L Ch R = 1 ,51013   ,485,485,485
BEGIN DESCRIPTION:
BEAVER CREEK 74.0
END DESCRIPTION:
XS GIS Cut Line= 3
       3709649.6     10688960.17      3709949.61     10689760.19
      3710299.59     10690460.15
#Sta/Elev= 30
    4113  363.86  4274.1  348.19  4422.7  338.68  4494.8  336.47  4555.4  337.85
  4665.7  334.14  4701.3  330.67  4720.9  330.46  4726.2  327.93  4751.2  326.11
  4756.5  323.33  4786.8   320.5  4860.6  317.05  4903.3  312.44  4975.8  314.37
  4998.2  307.44  5003.8  309.62  5017.5  307.28  5020.3  306.78  5023.5  307.28
  5026.1  310.74  5056.9  313.67    5205  312.09  5280.5  321.02  5311.2  322.06
  5445.4  335.48  5512.5  340.25  5629.9  353.22  5638.2  352.69    5750  360.76
#Mann= 3 ,-1 , 0
    4113     .12       0  5017.5     .07       0  5023.5     .12       0
Bank Sta=4975.8,5056.9
XS Rating Curve= 0 ,0
Exp/Cntr=0.3,0.1

Type RM Length L Ch R = 1 ,50528   ,726,726,726
BEGIN DESCRIPTION:
BEAVER CREEK 73.0
END DESCRIPTION:
XS GIS Cut Line= 3
       3709560.1     10689153.57      3709638.22      10690125.8
      3709169.48     10690854.96
#Sta/Elev= 30
  4123.4  349.39  4177.5  345.77  4230.4  345.86    4421  339.24  4531.3  330.84
  4591.5  329.39  4621.6  326.69  4701.9  324.06  4902.5  312.14  4972.8  312.61
  4992.8  304.46  4999.8  304.12  5002.6  303.62  5005.8  304.12  5012.9  307.06
  5022.9  312.98  5032.9  312.16    5043  313.25    5318  312.22  5448.7  313.73
  5555.7  312.52    5607     315  5637.4  318.75  5686.5  321.98  5694.8  323.62
  5722.2  325.09  5767.4  329.83  5846.1  337.15  5898.7  344.86  5965.6  353.95
#Mann= 5 ,-1 , 0
  4123.4     .12       0  4999.8     .07       0  5005.8     .12       0
  5767.4     .16       0  5898.7     .12       0
Bank Sta=4972.8,5022.9
XS Rating Curve= 0 ,0
Exp/Cntr=0.3,0.1

Type RM Length L Ch R = 1 ,49802   ,503,503,503
BEGIN DESCRIPTION:
BEAVER CREEK 72.0
END DESCRIPTION:
XS GIS Cut Line= 2
      3709178.15     10688919.21      3708935.16     10690715.65
#Sta/Elev= 30
    3818  351.26  3859.4   347.1  3916.9  338.53  4010.7   330.3  4072.3  320.22
  4121.7  318.92  4131.8  316.27  4162.1  317.19  4283.2  308.81  4908.8  310.34
  4969.4  311.54  4979.5  310.19  4989.5  303.58  4996.6  302.67  4999.4  302.17
  5002.6  302.67  5009.7  307.53  5019.8  310.74  5114.2  308.79  5171.2  311.23
  5264.5  319.67  5322.6  323.42    5332  322.79  5337.1  324.52    5373  327.74
  5403.3   328.5  5414.8  331.63  5473.9  335.76  5487.4  337.94  5630.8  347.36
#Mann= 3 ,-1 , 0
    3818     .12       0  4996.6     .07       0  5002.6     .12       0
Bank Sta=4969.4,5019.8
XS Rating Curve= 0 ,0
Exp/Cntr=0.3,0.1

Type RM Length L Ch R = 1 ,49299   ,894,894,894
BEGIN DESCRIPTION:
Mapping XS 871e6e66
END DESCRIPTION:
XS GIS Cut Line= 2
      3708902.42     10688617.64      3708652.58     10690236.38
#Sta/Elev= 30
  3881.7  347.19  3931.3  342.64  3999.5  339.78  4106.9  332.51  4130.9  334.54
  4147.4  333.49  4199.1  336.17  4238.4  335.89  4257.1  334.15  4299.1  325.27
  4319.4  320.19  4325.3  316.21  4339.6  313.04    4370   310.1  4410.4  310.34
  4501.5  307.31    4982  310.39  4994.3  303.06    4997  302.56  5000.3  303.06
  5027.7  309.49  5068.1  309.81  5098.5  314.69  5161.4  320.21  5180.8  322.07
    5230  327.87  5329.2  336.12    5376  338.84  5432.4  345.26  5519.6  347.72
#Mann= 6 ,-1 , 0
  3881.7     .12       0  4994.3     .07       0  5000.3     .12       0
  5161.4     .16       0  5180.8     .12       0  5329.2     .16       0
Bank Sta=4982,5027.7
XS Rating Curve= 0 ,0
Exp/Cntr=0.3,0.1

Type RM Length L Ch R = 1 ,48405   ,457,457,457
BEGIN DESCRIPTION:
BEAVER CREEK 71.0
END DESCRIPTION:
XS GIS Cut Line= 2
      3708171.21     10688823.69      3708266.64      10690576.2
#Sta/Elev= 30
    4532  350.58  4538.5  348.25  4550.9  347.34  4668.7  333.95  4738.8  329.41
  4788.9  322.47    4869  314.68  4958.2   306.5  4979.2  306.86  4996.2  298.56
  4998.9  298.06  5002.2  298.56  5009.2  305.79  5019.2  307.55  5150.3  307.03
  5189.5   305.8  5199.5  303.76  5219.5  306.01  5439.8   308.1  5600.1   306.8
  5770.3  308.22  5810.4  306.82  5830.4   308.9  5878.7  308.93  5892.5  310.44
  6000.7  315.27  6060.8  320.25  6091.9  324.67    6201  336.58  6287.1  348.87
#Mann= 6 ,-1 , 0
    4532     .16       0  4550.9     .12       0  4996.2     .07       0
  5002.2     .12       0  5892.5     .16       0  6091.9     .12       0
Bank Sta=4979.2,5019.2
XS Rating Curve= 0 ,0
Exp/Cntr=0.3,0.1

Type RM Length L Ch R = 1 ,47948   ,895,895,895
BEGIN DESCRIPTION:
Mapping XS f91bc3bb
END DESCRIPTION:
XS GIS Cut Line= 2
      3707996.16     10688898.91      3707657.91      10690496.5
#Sta/Elev= 30
  4372.4  352.28  4537.3  356.13  4595.2  351.98  4617.6  350.17  4622.7  352.22
  4667.3  345.26  4672.4     347    4711  337.36    4717  333.72  4722.1  336.58
  4731.5  334.79  4761.6  322.82  4766.7  324.63    4803  304.62  4823.5  306.97
  4893.4  305.84  4966.6  306.04    4987  299.97    5007  297.42  5009.8  296.92
    5013  297.42  5027.9  306.49    5154  305.35    5171  302.83  5191.4  304.86
  5685.3     305  5804.7  317.49    5896  338.46    5933   342.7  6005.4  351.72
#Mann= 7 ,-1 , 0
  4372.4     .12       0  4595.2     .16       0  4893.4     .12       0
    5007     .07       0    5013     .12       0    5896     .16       0
    5933     .12       0
Bank Sta=4966.6,5027.9
XS Rating Curve= 0 ,0
Exp/Cntr=0.3,0.1

Type RM Length L Ch R = 1 ,47053   ,690,690,690
BEGIN DESCRIPTION:
Mapping XS 3a522033
END DESCRIPTION:
XS GIS Cut Line= 4
      3707766.98     10688716.66      3707121.16     10689424.97
      3707131.58     10690023.93      3707334.67      10690414.5
#Sta/Elev= 30
  3917.9  343.92  4251.1   316.4  4428.1  305.01  4491.6  302.72  4711.2  302.09
  4971.7  304.01  4998.7   294.6  5001.4   294.1  5004.7   294.6  5011.7  303.16
  5075.7  302.24  5111.7  308.87  5171.7  309.74  5221.7   314.7  5281.7  325.58
  5381.7  323.84  5475.5  331.55  5485.1  335.71  5561.4   338.7    5590  342.95
  5612.1  341.94  5628.6  344.45  5634.2   342.4  5650.7  345.48  5700.6     345
    5717  347.15  5722.7  345.25  5739.1  348.73  5761.3  349.69  5915.7  348.59
#Mann= 3 ,-1 , 0
  3917.9     .12       0  4998.7     .07       0  5004.7     .12       0
Bank Sta=4971.7,5011.7
XS Rating Curve= 0 ,0
Exp/Cntr=0.3,0.1

Type RM Length L Ch R = 1 ,46363   ,392,392,392
BEGIN DESCRIPTION:
BEAVER CREEK 68.0
END DESCRIPTION:
XS GIS Cut Line= 4
      3707615.66     10688632.74       3706478.5     10689622.33
      3706495.86     10689761.22      3707224.79     10690299.24
#Sta/Elev= 30
  3431.8  350.78  3483.7  344.06  3491.3  338.07  3519.4  328.83  3554.9  323.94
  3618.6  322.02  3859.7  304.01  3972.7  301.81  4426.5  301.73  4483.5  300.08
  4504.4  302.35  4774.1   301.8    4831  299.68  4977.4  302.34  4990.5  300.57
  4994.6  292.01  4997.3  291.51  5000.6  292.01  5027.8  301.93    5159  299.95
  5545.3  301.69  5618.3  307.35    5681  314.46    5704  319.46  5724.9  328.85
  5789.6  343.14  5875.2  348.96  5889.9   351.5  5916.9  349.35  5985.2  348.71
#Mann= 3 ,-1 , 0
  3431.8     .12       0  4994.6     .07       0  5000.6     .12       0
Bank Sta=4977.4,5027.8
XS Rating Curve= 0 ,0
Exp/Cntr=0.3,0.1

Type RM Length L Ch R = 1 ,45971   ,559,559,559
BEGIN DESCRIPTION:
BEAVER CREEK 67.0
END DESCRIPTION:
XS GIS Cut Line= 3
      3707749.62     10688260.18      3706199.61     10689710.19
      3705399.57      10689860.2
#Sta/Elev= 30
  2856.5  367.34    2918   365.2  2955.4  365.64  2976.9  361.59  3045.5   357.8
  3149.1  348.87  3217.3  342.11  3245.2   336.5  3302.3  319.38  3373.1  311.11
  3592.4  301.99  4200.6     301  4222.1  299.23  4236.3  301.86  4667.6  299.85
  4752.6  301.98  4787.8  299.79  4823.4  302.07  4965.1  301.16  4971.9  298.56
  4975.6  293.31  5002.3  290.92    5005  290.42  5008.3  290.92  5010.4  298.94
  5107.1   299.1  5253.7  299.17  5388.5  304.75    5681  321.08    5793  330.25
#Mann= 8 ,-1 , 0
  2856.5     .12       0    2918     .16       0  3045.5     .12       0
  3149.1     .16       0  3245.2     .12       0  5002.3     .07       0
  5008.3     .12       0  5107.1     .05       0
Bank Sta=4965.1,5010.4
XS Rating Curve= 0 ,0
Exp/Cntr=0.3,0.1

Type RM Length L Ch R = 1 ,45412   ,542,542,542
BEGIN DESCRIPTION:
BEAVER CREEK 66.0
END DESCRIPTION:
XS GIS Cut Line= 3
       3707449.6     10688260.19      3705899.61     10689260.19
      3705263.87     10689387.83
#Sta/Elev= 30
  3166.9  347.16  3180.4  344.29  3225.9  339.29  3237.9  335.45  3262.1  328.89
  3289.3  324.14  3369.2  317.65  3594.9  305.29  3666.7  305.72  3724.9  302.32
  4223.8  298.36  4244.9  300.01    4476  298.94    4635  301.31  4678.3  299.14
  4722.7  300.23  4844.9  297.66  4975.8  298.78  4982.8  290.94  5000.9  290.43
  5003.6  289.93  5006.9  290.43  5031.8  297.67    5070   297.6  5291.4  308.98
  5489.9  331.52  5501.1  334.63  5521.5   337.1  5591.7  340.97  5659.9  348.36
#Mann= 5 ,-1 , 0
  3166.9     .16       0  3237.9     .12       0  5000.9     .07       0
  5006.9     .12       0    5070     .05       0
Bank Sta=4975.8,5031.8
XS Rating Curve= 0 ,0
Exp/Cntr=0.3,0.1

Type RM Length L Ch R = 1 ,44870   ,505,505,505
BEGIN DESCRIPTION:
BEAVER CREEK 65.0
END DESCRIPTION:
XS GIS Cut Line= 3
      3706649.64     10688010.16      3705849.61     10688760.19
      3705499.64     10688960.17
#Sta/Elev= 30
  3894.9  332.12    3995  323.24    4072  311.74  4220.5  302.79  4326.5  302.91
  4340.4  300.88  4482.3  297.94  4970.3  296.83  4984.4  289.65  4996.4  287.54
  4999.2  287.04  5002.4  287.54  5014.6   289.9    5021  296.33  5026.8  297.17
  5123.3  297.49  5139.1  299.56  5144.8  297.75  5181.1  298.35  5233.4  298.37
  5284.5  303.03    5314   311.1  5327.7  318.39    5337  319.47  5349.3  325.59
  5360.3   327.4  5371.6  334.27    5381  336.29  5391.8   343.2  5394.6   343.2
#Mann= 6 ,-1 , 0
  3894.9     .16       0    3995     .12       0  4996.4     .07       0
  5002.4     .12       0  5181.1     .05       0  5360.3     .16       0
Bank Sta=4970.3,5026.8
XS Rating Curve= 0 ,0
Exp/Cntr=0.3,0.1

Type RM Length L Ch R = 1 ,44365   ,524,524,524
BEGIN DESCRIPTION:
BEAVER CREEK 64.0
END DESCRIPTION:
XS GIS Cut Line= 3
      3706549.63     10687610.17      3705749.61     10688310.19
      3705349.59     10689010.22
#Sta/Elev= 30
  3952.4  331.62  3980.4  328.35    4045  313.25  4072.5   310.5  4172.1  299.19
  4229.1  295.97  4979.8  296.13  4987.4  295.43  4994.1  287.92  4998.7     287
  5001.4   286.5  5004.7     287  5018.3  288.14  5023.4  293.93  5050.7  296.75
  5178.2   298.8  5507.1  299.79  5615.1  305.14  5668.3  315.39  5674.1  314.45
  5689.9  321.33  5711.5  324.57    5718  328.86  5727.4  330.65  5733.1  328.38
    5749  334.28  5754.7  331.29  5759.9  333.02  5789.6  336.81  5821.7  339.09
#Mann= 7 ,-1 , 0
  3952.4     .16       0  4072.5     .12       0  4998.7     .07       0
  5004.7     .12       0  5178.2     .05       0  5759.9     .16       0
  5789.6     .05       0
Bank Sta=4979.8,5050.7
XS Rating Curve= 0 ,0
Exp/Cntr=0.3,0.1

Type RM Length L Ch R = 1 ,43841   ,562,562,562
BEGIN DESCRIPTION:
BEAVER CREEK 63.0
END DESCRIPTION:
XS GIS Cut Line= 3
      3706649.61     10687460.19      3705549.61     10687860.19
       3704749.6      10688560.2
#Sta/Elev= 30
  3825.4  348.52  3840.7  348.52  3889.2  338.97  3942.4  332.02  3995.6  318.17
  4035.2  313.34  4144.6  299.38  4229.7  297.35  4451.2  295.01  4715.9  296.09
  4751.8  294.54  4761.8  291.49  4771.8     295  4807.7  296.25  4963.9  296.87
  4974.6  294.48  4980.6  287.83    5000  285.06  5002.7  284.56    5006  285.06
  5017.2  286.57  5023.9  289.88  5031.5  299.05  5038.1  297.02  5095.1  295.41
    5235  296.97  5973.9  307.68  6023.3  310.14  6051.8  314.04  6058.9  316.92
#Mann= 5 ,-1 , 0
  3825.4     .16       0  4035.2     .12       0    5000     .07       0
    5006     .12       0    5235     .05       0
Bank Sta=4963.9,5031.5
XS Rating Curve= 0 ,0
Exp/Cntr=0.3,0.1

Type RM Length L Ch R = 1 ,43279   ,515,515,515
BEGIN DESCRIPTION:
BEAVER CREEK 62.0
END DESCRIPTION:
XS GIS Cut Line= 3
      3706349.62     10686660.17      3705549.61     10687460.19
      3703949.65     10688260.17
#Sta/Elev= 30
  3885.2  315.87    4564  295.41  4875.2  293.62  4974.2  294.87  5002.5  285.04
  5010.1  284.91  5012.8  284.41  5016.1  284.91  5019.4  284.91  5030.6  292.43
    5039  295.59  5329.9  294.35    5584  294.33  5947.4  299.02  6045.2  302.92
  6080.8  308.54  6112.3  313.57    6143  322.44  6187.7  329.44  6224.6  332.48
  6254.8  335.68  6327.5  333.93  6411.3  335.27  6590.2  355.34  6662.9  360.34
  6724.4  369.08  6752.3  369.71  6774.7  372.28  6783.1  375.32  6805.4  376.84
#Mann= 6 ,-1 , 0
  3885.2     .12       0  5010.1     .07       0  5016.1     .12       0
  5329.9     .05       0  6080.8     .16       0  6224.6     .05       0
Bank Sta=4974.2,5039
XS Rating Curve= 0 ,0
Exp/Cntr=0.3,0.1

Type RM Length L Ch R = 1 ,42764   ,493,493,493
BEGIN DESCRIPTION:
BEAVER CREEK 61.0
END DESCRIPTION:
XS GIS Cut Line= 3
       3705749.6      10686210.2      3705299.61     10687010.19
      3704499.63     10687810.17
#Sta/Elev= 30
  4045.5   354.8  4096.8  350.92  4102.8  348.74  4140.1  345.02  4156.1  339.86
  4199.4  333.52  4206.1  330.06    4252  320.74  4258.7  317.64  4280.4  315.71
  4286.4  312.19  4420.6  292.88  4977.5  294.19  5002.8  284.55  5005.5  284.05
  5008.8  284.55  5048.2  296.33  5090.6  293.22  5422.8  293.75  5474.9  293.54
    5727  293.82  5755.3  295.99  5854.3  295.63  5882.6  298.48  5910.9  296.49
  5967.5   296.8  6009.9  303.21  6038.2  312.06  6066.4  323.93  6094.7  330.39
#Mann= 5 ,-1 , 0
  4045.5     .12       0  5002.8     .07       0  5008.8     .12       0
  5422.8     .07       0  5474.9     .05       0
Bank Sta=4977.5,5048.2
XS Rating Curve= 0 ,0
Exp/Cntr=0.3,0.1

Type RM Length L Ch R = 1 ,42271   ,515,515,515
BEGIN DESCRIPTION:
BEAVER CREEK 60.0
END DESCRIPTION:
XS GIS Cut Line= 3
      3705549.58     10686210.22      3705049.61     10686610.19
      3703899.61     10688160.19
#Sta/Elev= 30
  4346.5  345.84  4388.9  342.94  4474.5  329.74  4502.5  323.64  4538.6  311.48
  4560.2  307.49  4574.6  302.21  4616.2   292.1  4801.9  291.47  4958.8  293.64
  4979.6  291.75  4983.6   287.4  5005.7   283.6  5008.4   283.1  5011.7   283.6
  5050.4  293.47  5173.8  293.02  5995.4  293.78  6172.9  300.97  6373.2  320.65
  6458.8  334.31  6523.5  348.31  6530.8  352.37  6558.9  356.72    6753  364.91
  6803.1   370.1    6867  382.16  6888.6  384.22  6894.9  386.84  6916.8  388.59
#Mann= 4 ,-1 , 0
  4346.5     .12       0  5005.7     .07       0  5011.7     .12       0
  5173.8     .05       0
Bank Sta=4958.8,5050.4
XS Rating Curve= 0 ,0
Exp/Cntr=0.3,0.1

Type RM Length L Ch R = 1 ,41756   ,624,624,624
BEGIN DESCRIPTION:
BEAVER CREEK 59.0
END DESCRIPTION:
XS GIS Cut Line= 3
      3705599.59     10686160.19      3704799.61     10686160.19
      3703199.61     10686060.19
#Sta/Elev= 30
  4227.6  350.26  4297.6  338.86  4407.6  325.45  4477.6  312.02  4627.6  292.65
  4887.6  290.55  4977.6  292.55  4987.6  291.95  4997.6   283.9  5014.6  283.21
  5017.3  282.71  5020.6  283.21  5025.1   286.4  5030.1   286.4  5037.6  290.76
  5047.6  292.91  5087.7  290.25  5270.6  291.41  5298.1  290.29  5591.4  293.51
  6099.7  296.77  6182.8  299.58  6300.1  312.62  6392.7   319.4  6420.3  330.18
  6433.4  333.15  6470.4  343.69  6511.7  350.08  6590.6  362.37  6630.7  365.33
#Mann= 7 ,-1 , 0
  4227.6     .12       0  5014.6     .07       0  5020.6     .12       0
  5591.4     .05       0  6182.8     .12       0  6433.4     .16       0
  6511.7     .12       0
Bank Sta=4977.6,5047.6
XS Rating Curve= 0 ,0
Exp/Cntr=0.3,0.1

Type RM Length L Ch R = 1 ,41132   ,103,103,103
BEGIN DESCRIPTION:
BEAVER CREEK 58.0
END DESCRIPTION:
XS GIS Cut Line= 2
      3705735.31     10685661.48      3703315.12      10685546.9
#Sta/Elev= 30
  3824.2  349.07  3990.1  330.04  4040.1  329.93  4130.2   314.9  4260.4  301.97
  4570.7  291.89  4871.1  290.24  4911.1  286.02  4941.1  286.27  4971.2  290.85
  5007.4  283.29  5010.1  282.79  5013.4  283.29  5021.2  284.08  5031.2  290.87
  5061.3  288.65  5311.6  291.44  5543.9  301.38  5642.8  301.69  5858.7  312.26
  5863.7  310.02  5932.3  313.18  5942.3  317.22  5951.5  316.59  6069.6  323.25
  6074.6  319.76  6137.2  321.05  6172.5  322.01  6202.6  329.96  6247.1   334.8
#Mann= 7 ,-1 , 0
  3824.2     .05       0  5007.4     .04       0  5013.4     .05       0
  5543.9     .08       0  5642.8     .05       0  5951.5     .16       0
  6137.2     .05       0
Bank Sta=4971.2,5031.2
XS Rating Curve= 0 ,0
Exp/Cntr=0.3,0.1

Type RM Length L Ch R = 1 ,41029   ,879,879,879
BEGIN DESCRIPTION:
BEAVER CREEK 57.0
END DESCRIPTION:
XS GIS Cut Line= 2
      3705710.96     10685550.37      3703343.71     10685456.65
#Sta/Elev= 30
  3838.8  342.97  4000.3  324.02  4010.3  324.39  4140.4  310.66  4230.5  303.71
  4550.7  292.73  4700.8  292.35  4780.9  290.02    4871  290.92    4911  288.09
    4951   291.4  4983.5   291.6    4991  285.53  5018.1   283.2  5020.8   282.7
  5024.1   283.2  5035.4  287.37  5051.1  290.26  5281.3  288.85  5411.4  291.22
  5486.5  296.72  5522.8  297.07  5551.5   297.2  5581.5  300.01  5611.5  298.56
  5791.7  303.79  6031.9  312.88  6041.9  314.79  6091.9  314.98  6207.9  324.45
#Mann= 5 ,-1 , 0
  3838.8     .05       0  5018.1     .03       0  5024.1     .05       0
  5035.4     .12       0  5522.8     .05       0
Bank Sta=4983.5,5051.1
XS Rating Curve= 0 ,0
Exp/Cntr=0.3,0.1

Type RM Length L Ch R = 1 ,40150   ,535,535,535
BEGIN DESCRIPTION:
BEAVER CREEK 56.0
END DESCRIPTION:
XS GIS Cut Line= 3
      3705449.66     10684610.18      3703899.61     10685010.19
      3703276.93     10685442.74
#Sta/Elev= 30
  3408.2  361.65  3424.7  361.02  3553.2  338.58  3664.8  327.43    3670  325.26
  3705.5  323.57  3769.7  312.22  3779.6  312.12  3976.3     295    4107  288.54
  4327.4  286.68  4864.1  287.59  4966.3  290.21    4978  288.67  4991.3  281.56
  5003.4  281.51  5006.2  281.01  5009.4  281.51  5012.1  281.51  5016.5  287.55
  5031.3  289.97    5056  288.78  5094.3  287.78  5210.3  290.77  5252.5  295.01
  5469.6  303.17    5583  312.56  5669.5  316.08  5684.3  319.18  5767.2  326.08
#Mann= 7 ,-1 , 0
  3408.2     .05       0  3424.7     .12       0  3779.6     .05       0
  4966.3     .12       0  5003.4     .07       0  5009.4     .12       0
    5056     .05       0
Bank Sta=4966.3,5031.3
XS Rating Curve= 0 ,0
Exp/Cntr=0.3,0.1
