--- CATFISH CREEK.prj (project) ---

Proj Title=CATFISH CREEK Base Level Engineering
Current Plan=p01
Default Exp/Contr=0.3,0.1
English Units
Geom File=g01
Flow File=f01
Plan File=p01
Y Axis Title=Elevation
X Axis Title(PF)=Main Channel Distance
X Axis Title(XS)=Station
BEGIN DESCRIPTION:
CATFISH CREEK
END DESCRIPTION:
DSS Export Rating Curves= 0
DSS Export Rating Curve Sorted= 0
DSS Export Volume Flow Curves= 0
DXF OffsetX= 0
DXF OffsetY= 0
DXF ScaleX= 1
DXF ScaleY= 10

--- CATFISH CREEK.p01 (plan) ---

Plan Title=Multiple Run
Short Identifier=Multiple
Geom File=g01
Flow File=f01
Subcritical Flow
K Sum by GR= 0
Std Step Tol= 0.01
Critical Tol= 0.01
Num of Std Step Trials= 20
Max Error Tol= 0.3
Flow Tol Ratio= 0.001
Split Flow NTrial= 30
Split Flow Tol= 0.02
Split Flow Ratio= 0.02
Log Output Level= 0
Friction Slope Method= 1
Unsteady Friction Slope Method= 2
Unsteady Bridges Friction Slope Method= 1
Parabolic Critical Depth
Global Vel Dist=  1 , 1 , 1
Global Log Level= 0
CheckData=True
Encroach Param= -1, 0, 0, 0
BEGIN DESCRIPTION:
Multiple Run
END DESCRIPTION:

--- CATFISH CREEK.f01 (steady flow) ---

Flow Title=Multiple
Program Version=4.10
Number of Profiles= 7
Profile Names=10-year,25-year,50-year,1pct_min,100-year,1pct_plu,500-year
River Rch & RM=CATFISH CREEK,Reach-1         ,233951
     816    1123    1379    1243    1680    2273    2499
River Rch & RM=CATFISH CREEK,Reach-1         ,230204
     982    1367    1692    1535    2075    2807    3131
River Rch & RM=CATFISH CREEK,Reach-1         ,228153
    1020    1413    1742    1573    2128    2878    3181
River Rch & RM=CATFISH CREEK,Reach-1         ,222835
    1339    1889    2358    2155    2914    3941    4461
River Rch & RM=CATFISH CREEK,Reach-1         ,220815
    1744    2488    3130    2879    3893    5265    6040
River Rch & RM=CATFISH CREEK,Reach-1         ,218369
    1767    2519    3167    2911    3937    5324    6101
River Rch & RM=CATFISH CREEK,Reach-1         ,215829
    1943    2777    3497    3218    4352    5886    6761
River Rch & RM=CATFISH CREEK,Reach-1         ,212564
    1926    2745    3450    3167    4283    5793    6624
River Rch & RM=CATFISH CREEK,Reach-1         ,209345
    2625    3790    4805    4447    6014    8134    9451
River Rch & RM=CATFISH CREEK,Reach-1         ,208032
    3601    5263    6730    6277    8488   11480   13544
River Rch & RM=CATFISH CREEK,Reach-1         ,207451
    3601    5263    6730    6277    8488   11480   13544
River Rch & RM=CATFISH CREEK,Reach-1         ,203983
    4646    6838    8783    8225   11123   15043   17888
River Rch & RM=CATFISH CREEK,Reach-1         ,203251
    4646    6838    8783    8225   11123   15043   17888
River Rch & RM=CATFISH CREEK,Reach-1         ,198857
    4658    6839    8770    8198   11087   14994   17766
River Rch & RM=CATFISH CREEK,Reach-1         ,194134
    4622    6776    8682    8106   10963   14826   17529
River Rch & RM=CATFISH CREEK,Reach-1         ,191292
    4737    6949    8905    8317   11248   15211   17993
River Rch & RM=CATFISH CREEK,Reach-1         ,190671
    5276    7747    9936    9284   12556   16980   20101
River Rch & RM=CATFISH CREEK,Reach-1         ,183700
    5249    7698    9865    9208   12453   16842   19899
River Rch & RM=CATFISH CREEK,Reach-1         ,182085
    5390    7898   10115    9435   12760   17257   20358
River Rch & RM=CATFISH CREEK,Reach-1         ,181564
    5390    7898   10115    9435   12760   17257   20358
River Rch & RM=CATFISH CREEK,Reach-1         ,177844
    5478    8025   10276    9584   12961   17528   20670
River Rch & RM=CATFISH CREEK,Reach-1         ,174496
    5677    8315   10645    9925   13422   18151   21388
River Rch & RM=CATFISH CREEK,Reach-1         ,173482
    5677    8315   10645    9925   13422   18151   21388
River Rch & RM=CATFISH CREEK,Reach-1         ,170604
    5936    8698   11140   10388   14048   18998   22395
River Rch & RM=CATFISH CREEK,Reach-1         ,165153
    5973    8744   11192   10429   14104   19073   22451
River Rch & RM=CATFISH CREEK,Reach-1         ,162138
    5947    8698   11124   10358   14008   18944   22266
River Rch & RM=CATFISH CREEK,Reach-1         ,158941
    8480   12511   16104   15085   20400   27589   32811
River Rch & RM=CATFISH CREEK,Reach-1         ,153099
    8465   12476   16047   15021   20314   27472   32622
River Rch & RM=CATFISH CREEK,Reach-1         ,151249
    8459   12462   16025   14995   20279   27425   32545
River Rch & RM=CATFISH CREEK,Reach-1         ,149553
    8720   12854   16534   15478   20932   28308   33620
River Rch & RM=CATFISH CREEK,Reach-1         ,148796
    8794   12967   16683   15620   21124   28568   33940
River Rch & RM=CATFISH CREEK,Reach-1         ,145872
    8685   12779   16418   15349   20758   28073   33254
River Rch & RM=CATFISH CREEK,Reach-1         ,139904
    8644   12704   16307   15232   20599   27858   32940
River Rch & RM=CATFISH CREEK,Reach-1         ,135684
    8676   12745   16355   15272   20654   27932   33009
River Rch & RM=CATFISH CREEK,Reach-1         ,133898
    8676   12745   16355   15272   20654   27932   33009
River Rch & RM=CATFISH CREEK,Reach-1         ,129986
   14684   21657   27884   26096   35292   47728   56604
River Rch & RM=CATFISH CREEK,Reach-1         ,123003
   14536   21414   27549   25761   34839   47116   55785
River Rch & RM=CATFISH CREEK,Reach-1         ,121394
   14578   21467   27609   25811   34907   47207   55867
River Rch & RM=CATFISH CREEK,Reach-1         ,120515
   14578   21467   27609   25811   34907   47207   55867
River Rch & RM=CATFISH CREEK,Reach-1         ,119185
   14798   21765   27971   26131   35339   47792   56482
River Rch & RM=CATFISH CREEK,Reach-1         ,113634
   14704   21604   27746   25902   35029   47373   55905
River Rch & RM=CATFISH CREEK,Reach-1         ,108759
   14586   21412   27482   25640   34675   46894   55273
River Rch & RM=CATFISH CREEK,Reach-1         ,105936
   14530   21310   27333   25485   34466   46611   54870
River Rch & RM=CATFISH CREEK,Reach-1         ,103209
   14543   21320   27338   25481   34460   46603   54825
River Rch & RM=CATFISH CREEK,Reach-1         ,102597
   14543   21320   27338   25481   34460   46603   54825
River Rch & RM=CATFISH CREEK,Reach-1         ,99465
   14598   21386   27411   25539   34538   46709   54903
River Rch & RM=CATFISH CREEK,Reach-1         ,98561
   14598   21386   27411   25539   34538   46709   54903
River Rch & RM=CATFISH CREEK,Reach-1         ,96762
   14647   21456   27499   25620   34648   46857   55077
River Rch & RM=CATFISH CREEK,Reach-1         ,96106
   14647   21456   27499   25620   34648   46857   55077
River Rch & RM=CATFISH CREEK,Reach-1         ,94707
   14647   21456   27499   25620   34648   46857   55077
River Rch & RM=CATFISH CREEK,Reach-1         ,93811
   14667   21471   27507   25617   34644   46851   55024
River Rch & RM=CATFISH CREEK,Reach-1         ,89290
   14597   21349   27333   25438   34402   46525   54569
River Rch & RM=CATFISH CREEK,Reach-1         ,83657
   14751   21566   27605   25686   34738   46979   55080
River Rch & RM=CATFISH CREEK,Reach-1         ,80095
   14580   21280   27208   25287   34197   46248   54096
River Rch & RM=CATFISH CREEK,Reach-1         ,74210
   14632   21357   27307   25380   34324   46419   54299
River Rch & RM=CATFISH CREEK,Reach-1         ,71228
   14632   21357   27307   25380   34324   46419   54299
River Rch & RM=CATFISH CREEK,Reach-1         ,70895
   14473   21100   26956   25032   33853   45783   53466
River Rch & RM=CATFISH CREEK,Reach-1         ,64644
   14302   20818   26566   24642   33326   45070   52513
River Rch & RM=CATFISH CREEK,Reach-1         ,56644
   16513   24048   30714   28521   38572   52164   60911
River Rch & RM=CATFISH CREEK,Reach-1         ,54848
   16513   24048   30714   28521   38572   52164   60911
River Rch & RM=CATFISH CREEK,Reach-1         ,52040
   16500   24007   30643   28438   38459   52011   60658
River Rch & RM=CATFISH CREEK,Reach-1         ,46803
   16441   23908   30505   28298   38270   51756   60311
River Rch & RM=CATFISH CREEK,Reach-1         ,43876
   16306   23688   30204   27999   37866   51209   59593
River Rch & RM=CATFISH CREEK,Reach-1         ,32816
   16320   23697   30205   27991   37855   51194   59532
River Rch & RM=CATFISH CREEK,Reach-1         ,28738
   16227   23542   29989   27773   37560   50796   58995
Boundary for River Rch & Prof#=CATFISH CREEK,Reach-1         , 1
Up Type= 0
Dn Type= 3
Dn Slope=0.0012
Boundary for River Rch & Prof#=CATFISH CREEK,Reach-1         , 2
Up Type= 0
Dn Type= 3
Dn Slope=0.0012
Boundary for River Rch & Prof#=CATFISH CREEK,Reach-1         , 3
Up Type= 0
Dn Type= 3
Dn Slope=0.0012
Boundary for River Rch & Prof#=CATFISH CREEK,Reach-1         , 4
Up Type= 0
Dn Type= 3
Dn Slope=0.0012
Boundary for River Rch & Prof#=CATFISH CREEK,Reach-1         , 5
Up Type= 0
Dn Type= 3
Dn Slope=0.0012
Boundary for River Rch & Prof#=CATFISH CREEK,Reach-1         , 6
Up Type= 0
Dn Type= 3
Dn Slope=0.0012
Boundary for River Rch & Prof#=CATFISH CREEK,Reach-1         , 7
Up Type= 0
Dn Type= 3
Dn Slope=0.0012
DSS Import GetInterval= 0
DSS Import GetPeak= 0
DSS Import FillOption= 0

--- CATFISH CREEK.g01 (geometry) ---

Geom Title=Existing Conditions
Program Version=4.10

River Reach=CATFISH CREEK   ,Reach-1
Reach XY= 30
      3727794.08     10769479.18        3729570.       10768374.
       3727816.5       10762342.        3722002.       10759903.
      3714794.25       10750731.      3713026.75       10751554.
      3706319.25       10747302.       3703614.5       10739656.
      3701139.25       10739181.        3696632.       10726194.
      3689038.25       10720393.       3686988.5       10721334.
      3683157.75       10717077.        3682989.       10713781.
       3680262.5       10714318.       3680509.5       10708166.
      3678690.25       10707295.        3680085.       10698341.
       3676680.5       10691275.        3681092.       10686964.
       3681911.5       10675810.       3678049.5       10672120.
      3678346.25       10664742.       3672857.5       10660467.
        3670716.       10651142.      3664537.25       10645057.
        3666123.       10642400.       3665771.5       10638215.
      3663037.25       10638258.      3663934.05     10635986.57

Type RM Length L Ch R = 1 ,233951  ,627,627,627
BEGIN DESCRIPTION:
CATFISH CREEK 242.0
END DESCRIPTION:
XS GIS Cut Line= 4
      3727719.17     10770015.74      3727891.03     10769726.72
      3727888.42     10769375.15       3727784.8     10769074.65
#Sta/Elev= 30
  4374.2  524.31  4376.8  523.94  4422.7  519.41  4428.5  517.12  4459.7  515.58
  4465.5  513.64  4481.1  514.17  4486.9  512.06  4523.9  507.67  4531.9  508.24
  4555.1  505.78  4576.6  502.73  4582.4  500.09    4635   493.9  4640.8  491.84
    4787  480.75    4927  470.53    4997   461.4  4999.8   460.9    5003   461.4
    5007  463.17    5017   461.4    5027  466.29  5042.7  467.72    5099  468.41
  5151.9  476.82  5223.9  485.02  5260.4  492.26  5322.8  499.97  5379.9  503.31
#Mann= 5 ,-1 , 0
  4374.2     .05       0  4376.8     .16       0    4997     .07       0
    5003     .16       0  5042.7     .05       0
Bank Sta=4787,5322.8
XS Rating Curve= 0 ,0
Exp/Cntr=0.3,0.1

Type RM Length L Ch R = 1 ,233324  ,435,435,435
BEGIN DESCRIPTION:
Mapping XS 8fde0b54
END DESCRIPTION:
XS GIS Cut Line= 3
      3728198.32     10770390.75      3728419.67     10769661.61
       3728310.3     10769047.07
#Sta/Elev= 30
  4290.2  511.02  4301.1  510.91  4380.2  503.58  4489.4  501.74  4604.9  487.62
  4802.9  466.24  4834.2  465.85  4866.3  462.93  4938.7  461.24    4991  460.08
    4997  458.14  4999.8  457.64    5003  458.14  5011.9  460.14  5038.9  460.43
  5094.3  459.44  5145.1  461.51  5198.1  464.47  5266.9  473.86  5305.9  473.81
    5311  476.82  5327.9  473.38  5348.2  474.83  5449.8  473.59    5483  476.65
  5500.6  484.88  5510.7  493.09  5520.9  495.18    5542  491.49  5676.4  504.04
#Mann= 7 ,-1 , 0
  4290.2     .05       0  4301.1      .1       0  4604.9     .12       0
  4866.3     .16       0    4997     .07       0    5003     .16       0
  5038.9     .05       0
Bank Sta=4938.7,5145.1
XS Rating Curve= 0 ,0
Exp/Cntr=0.3,0.1

Type RM Length L Ch R = 1 ,232889  ,636,636,636
BEGIN DESCRIPTION:
Mapping XS bf15db59
END DESCRIPTION:
XS GIS Cut Line= 2
      3729093.95     10770759.75      3728486.29     10768958.48
#Sta/Elev= 30
  3740.7  508.86  3782.5  508.96  3831.2  513.14  3862.7  511.76  3899.4  504.92
  3930.9  503.58  4088.5  483.62  4203.6  471.95  4373.5  462.92    4384  462.29
  4500.1  458.27  4827.3  458.38  4858.9  460.22  4864.5  457.04  4948.1  455.55
  4983.7  455.79    4997  455.09  4999.8  454.59    5003  455.09    5070  457.72
  5196.6  471.55  5217.8   475.3  5336.6  483.04  5362.8  483.83  5368.1  482.29
  5394.3  489.71  5418.3  487.82    5431  488.89  5583.1  507.37  5641.7  510.82
#Mann= 7 ,-1 , 0
  3740.7     .05       0  4373.5     .07       0    4384     .05       0
  4948.1     .16       0  4983.7     .05       0    4997     .03       0
    5003     .05       0
Bank Sta=4864.5,5070
XS Rating Curve= 0 ,0
Exp/Cntr=0.3,0.1

Type RM Length L Ch R = 1 ,232253  ,388,388,388
BEGIN DESCRIPTION:
Mapping XS 72d50cac
END DESCRIPTION:
XS GIS Cut Line= 2
      3729963.96     10769854.33      3728508.22     10768916.82
#Sta/Elev= 30
    4125  501.59    4154  500.02  4160.1   498.5  4232.8   491.6  4306.1  482.79
  4399.1   473.5  4529.2  469.85  4586.6  469.42  4680.4  464.37  4819.7  453.62
    4997  453.62  4999.8  453.12    5003  453.62  5215.8  453.62  5282.5   458.8
    5391  468.62  5439.6   475.6  5448.8  474.97  5475.9  479.94  5485.2  480.41
    5498  483.77  5542.6  486.19  5578.9  490.42  5584.9  492.09  5593.2  491.45
  5642.3  497.95  5651.5  497.54  5700.2  503.22  5751.2  506.73  5856.5  512.41
#Mann= 4 ,-1 , 0
    4125     .16       0  4306.1     .05       0    4997    .033       0
    5003     .05       0
Bank Sta=4586.6,5282.5
XS Rating Curve= 0 ,0
Exp/Cntr=0.3,0.1

Type RM Length L Ch R = 1 ,231865  ,617,617,617
BEGIN DESCRIPTION:
Mapping XS d6bfe56d
END DESCRIPTION:
XS GIS Cut Line= 3
      3729610.43     10769305.72      3729497.58      10769132.1
      3728785.81     10768528.83
#Sta/Elev= 30
  4615.9  473.79  4657.8  470.94  4684.9  467.73  4736.2  464.57  4793.6  458.64
  4814.7  457.09  4821.1  455.79  4836.8  455.22  4844.5  453.62    4997  453.62
  4999.8  453.12    5003  453.62  5205.9  453.62  5248.8  458.77  5298.2   461.3
  5312.5   463.6  5355.4  466.81  5361.9  468.29  5404.8  471.91  5468.5  475.14
  5546.5  481.78  5554.2  483.56  5595.9  488.01  5617.9  491.53  5638.8  493.13
  5681.6  500.31  5702.5   501.9  5724.5  505.82  5745.3  511.22    5756  512.27
#Mann= 3 ,-1 , 0
  4615.9     .05       0    4997    .033       0    5003     .05       0
Bank Sta=4793.6,5205.9
XS Rating Curve= 0 ,0
Exp/Cntr=0.3,0.1

Type RM Length L Ch R = 1 ,231248  ,350,350,350
BEGIN DESCRIPTION:
Mapping XS 8875f23c
END DESCRIPTION:
XS GIS Cut Line= 2
      3729881.71     10768483.41       3728816.2     10768342.35
#Sta/Elev= 30
  4677.6  465.86  4730.2  459.73  4737.7  458.24  4742.8  458.76  4770.5  456.24
  4780.6  453.62    4997  453.62  4999.8  453.12    5003  453.62  5264.8  453.62
    5285  455.08  5325.3  459.88  5395.9  466.11  5436.3   470.6  5476.6  476.74
  5486.7  477.57    5517  483.46  5547.2  486.74  5567.4  490.05  5587.6  495.11
  5617.8  498.15  5627.9  500.81    5638  501.81  5653.9  506.53  5658.9  506.25
  5668.3  509.18  5678.4  510.47  5688.4   512.9  5738.9  519.81  5752.4  520.76
#Mann= 3 ,-1 , 0
  4677.6     .05       0    4997    .033       0    5003     .05       0
Bank Sta=4780.6,5264.8
XS Rating Curve= 0 ,0
Exp/Cntr=0.3,0.1

Type RM Length L Ch R = 1 ,230898  ,183,183,183
BEGIN DESCRIPTION:
Mapping XS d8ea857d
END DESCRIPTION:
XS GIS Cut Line= 3
      3729971.55     10768253.87      3729704.65     10768054.23
      3729088.37     10768197.45
#Sta/Elev= 30
  4482.1  468.57  4493.7  468.49  4543.7  464.63  4549.9  463.47  4571.9  461.81
  4614.6  457.74  4621.9  456.84  4629.1  456.54  4632.4  453.62  4635.1  453.12
  4638.4  453.62  5292.8  453.62  5301.8   456.9  5306.9  456.09  5313.4  458.33
  5323.6  459.48  5344.2  463.87  5349.5  465.96  5354.7  465.81  5364.7  467.19
    5375  469.46  5385.2  470.58  5392.1  473.37  5397.3   473.3    5416  476.95
  5426.3  477.71  5434.8  479.09  5439.9  479.15  5444.9  480.13  5448.1  480.13
#Mann= 3 ,-1 , 0
  4482.1     .05       0  4632.4    .033       0  4638.4     .05       0
Bank Sta=4614.6,5313.4
XS Rating Curve= 0 ,0
Exp/Cntr=0.3,0.1

Type RM Length L Ch R = 1 ,230715  ,37,37,37
BEGIN DESCRIPTION:
Mapping XS 23b1d2b8
END DESCRIPTION:
XS GIS Cut Line= 3
      3730686.01     10767231.73      3729550.57     10767886.26
      3729033.45     10768149.16
#Sta/Elev= 30
  3626.1  497.28    3816  472.33  3852.5  469.32  3914.8   464.4  3967.9   463.6
  4025.9  460.45  4032.6  461.21  4171.9   458.2  4295.5  454.65  4332.8  455.38
  4345.6  453.62  4348.4  453.12  4351.6  453.62    5267  453.62  5283.6  455.96
  5289.3  453.87  5296.7  456.58  5311.5  456.47  5319.2  458.99  5350.4  464.81
  5364.1  465.87  5372.7  468.91  5417.2  477.06  5453.8  481.01  5461.7  483.27
  5476.2  484.75  5483.9  487.26  5498.7  488.67  5506.2  491.64  5516.8  493.52
#Mann= 5 ,-1 , 0
  3626.1     .05       0    3816     .08       0  3852.5     .05       0
  4345.6    .035       0  4351.6     .05       0
Bank Sta=4171.9,5319.2
XS Rating Curve= 0 ,0
Exp/Cntr=0.3,0.1

Type RM Length L Ch R = 1 ,230678  ,40,40,40
BEGIN DESCRIPTION:
Mapping XS 8e206fb9
END DESCRIPTION:
XS GIS Cut Line= 4
      3730609.99     10767173.18      3729726.78      10767722.2
      3729446.84     10767902.32      3729040.98     10768121.53
#Sta/Elev= 30
  3666.5  490.61  3800.2  473.46    3832   471.5  3961.3  465.23  3984.9  464.86
  3991.5  466.74  4122.6  465.64  4201.7  460.55  4259.5  459.41  4375.2  457.44
  4558.2  458.29  4716.4  457.04  4735.8  454.84  4738.5  454.34  4741.8  454.84
  4774.4  457.73  4804.3  455.75  4810.2  457.75  4840.6  455.98  4861.7  457.87
  4949.5  456.42  5115.7  457.98    5213  455.07  5278.7  456.97  5322.5  461.46
  5420.5  479.09  5426.2  477.98  5442.4  482.48  5448.1  480.89  5500.6  491.91
#Mann= 5 ,-1 , 0
  3666.5     .05       0  3800.2     .08       0    3832     .05       0
  4735.8     .03       0  4741.8     .05       0
Bank Sta=4558.2,4774.4
XS Rating Curve= 0 ,0
Exp/Cntr=0.3,0.1

Type RM Length L Ch R = 1 ,230638  ,73,73,73
BEGIN DESCRIPTION:
Mapping XS 7b535d31
END DESCRIPTION:
XS GIS Cut Line= 3
      3730609.62     10767143.19      3729472.44     10767839.82
       3729033.3     10768079.95
#Sta/Elev= 30
  3657.3  492.58  3772.4  476.97  3829.3  473.26  3829.5  473.26  3967.8  465.98
  4041.2  469.71  4389.4  459.91  4484.2  465.93  4600.3  457.71  4783.1  454.54
  4826.5  448.56  4869.1  450.18  4884.6  447.42  4890.4  449.75    4900  448.09
  4905.9  451.42  4921.3  447.43  4927.2  450.54  4935.6  447.85    4958  448.02
  4963.9  450.76  5019.8  446.76  5022.5  446.26  5025.8  446.76  5028.5  449.44
  5104.3  447.61    5110     450  5199.3  452.69  5442.1  483.56  5491.4  495.66
#Mann= 5 ,-1 , 0
  3657.3     .05       0  3829.3     .08       0  3829.5     .05       0
  5019.8     .03       0  5025.8     .05       0
Bank Sta=4783.1,5199.3
XS Rating Curve= 0 ,0
Exp/Cntr=0.3,0.1

Type RM Length L Ch R = 1 ,230565  ,361,361,361
BEGIN DESCRIPTION:
CATFISH CREEK 241.0
END DESCRIPTION:
XS GIS Cut Line= 2
      3730619.95     10767096.79      3728846.11     10768115.99
#Sta/Elev= 30
  3634.8  496.57  3762.1  478.31    3931  469.87  4070.4  473.79    4391  466.85
  4566.1  464.07  4751.9  453.37  4838.2  445.15  4875.5  448.16  5017.8  443.29
  5020.5  442.79  5023.8  443.29  5154.5  452.94    5337  473.89  5365.2  473.82
  5417.6  485.93  5476.5  490.49  5513.9   497.6  5519.6  502.82  5578.6  501.49
  5584.3  505.84  5594.4  503.42  5600.1  508.76  5615.9  503.48  5621.7  506.94
  5634.9  504.29  5643.3  508.37  5653.3  506.13  5659.1  510.48  5680.6  509.17
#Mann= 6 ,-1 , 0
  3634.8     .05       0    4391     .08       0  4566.1     .05       0
  5017.8     .03       0  5023.8     .05       0  5634.9     .08       0
Bank Sta=4751.9,5154.5
XS Rating Curve= 0 ,0
Exp/Cntr=0.3,0.1

Type RM Length L Ch R = 1 ,230204  ,403,403,403
BEGIN DESCRIPTION:
CATFISH CREEK 240.0
END DESCRIPTION:
XS GIS Cut Line= 2
      3730177.23     10766966.59      3728473.04     10767890.24
#Sta/Elev= 30
  3991.8  491.42  4340.8  490.58    4434  484.25  4537.6  484.55  4826.7  454.03
  4921.8   453.2  4930.4  449.05    4936  454.35  4944.5  452.86  4952.2  447.18
  4957.9  453.81  4974.1  447.68  4979.8  452.18    4990  449.84    4993  442.32
  4995.7  441.82    4999  442.32  5001.6  452.08  5012.1  448.89  5017.8  454.63
    5034     448  5039.7  452.27  5061.6  452.51  5077.7  446.79  5105.3  454.59
  5137.7  453.76  5319.9  476.44  5541.8  494.68  5705.3  496.38  5930.2  488.99
#Mann= 3 ,-1 , 0
  3991.8     .05       0    4993     .03       0    4999     .05       0
Bank Sta=4921.8,5105.3
XS Rating Curve= 0 ,0
Exp/Cntr=0.3,0.1

Type RM Length L Ch R = 1 ,229801  ,448,448,448
BEGIN DESCRIPTION:
CATFISH CREEK 239.0
END DESCRIPTION:
XS GIS Cut Line= 3
      3729649.59     10767110.19      3729299.61     10767060.19
      3729099.64     10767060.19
#Sta/Elev= 30
  4662.5  482.74    4665  482.74  4672.6  480.23  4682.7  478.81  4692.8  475.79
  4723.1  470.59  4763.5  465.55  4783.7  461.41    4814  458.12  4834.2  455.37
  4854.4   451.6  4874.6  449.31  4935.2  444.74  4985.7  441.82  4992.8  440.43
  4995.6  439.93  4998.8  440.43  5013.5   441.5    5036  440.73    5086  444.99
    5096  445.53    5116  448.27    5126  450.68    5136  451.42    5146  454.34
    5166  457.84    5176  458.82    5186  461.03    5206  463.82    5216  464.13
#Mann= 3 ,-1 , 0
  4662.5     .05       0  4992.8     .03       0  4998.8     .05       0
Bank Sta=4935.2,5086
XS Rating Curve= 0 ,0
Exp/Cntr=0.3,0.1

Type RM Length L Ch R = 1 ,229353  ,430,430,430
BEGIN DESCRIPTION:
CATFISH CREEK 238.0
END DESCRIPTION:
XS GIS Cut Line= 3
      3729549.64     10766410.16      3729249.61     10766660.19
      3729049.61     10766710.19
#Sta/Elev= 30
  4631.8  482.07  4659.8  480.73    4682  477.74  4696.3  474.44  4717.1  471.67
  4723.6  469.47  4731.4  468.91  4737.9  466.92  4760.1  464.38  4766.6  462.07
  4780.9  461.02    4788  459.05  4801.7  458.07  4838.2  452.26  4866.1  449.68
  4887.6  446.42  4951.4  440.66  4967.9  439.11  5055.2  438.98  5070.9  438.76
  5073.6  438.26  5076.9  438.76    5128   440.1  5135.7  441.76  5156.4  443.77
  5169.2  447.77  5197.6  452.96  5205.3  456.66  5218.2  456.28  5228.5  457.35
#Mann= 5 ,-1 , 0
  4631.8     .05       0  4967.9     .16       0  5055.2     .05       0
  5070.9     .07       0  5076.9     .05       0
Bank Sta=4951.4,5135.7
XS Rating Curve= 0 ,0
Exp/Cntr=0.3,0.1

Type RM Length L Ch R = 1 ,228923  ,702,702,702
BEGIN DESCRIPTION:
CATFISH CREEK 237.0
END DESCRIPTION:
XS GIS Cut Line= 3
      3729399.58     10766210.19      3729099.61     10766260.19
       3728299.6     10766710.19
#Sta/Elev= 30
    4697  470.82  4724.9  465.84  4757.8  461.39  4778.1  456.89  4798.4     455
  4818.6  450.69  4851.6  447.31  4859.2  445.87  4899.7  442.23  4907.3  440.81
  4912.4  441.86    4920  439.26  4940.3  436.96  5006.1  436.18  5008.8  435.68
  5012.1  436.18  5024.1  437.04  5058.5  436.23  5073.8  436.66    5100  436.54
  5413.8  436.97  5478.9  439.36  5484.6  438.95  5500.5  440.01  5506.3  439.55
  5551.8  440.63  5655.1  443.82  5758.4  448.69    5896  459.63    5919   460.6
#Mann= 5 ,-1 , 0
    4697     .05       0  5006.1    .035       0  5012.1     .05       0
  5073.8     .16       0    5100     .05       0
Bank Sta=4912.4,5551.8
XS Rating Curve= 0 ,0
Exp/Cntr=0.3,0.1

Type RM Length L Ch R = 1 ,228221  ,68,68,68
BEGIN DESCRIPTION:
CATFISH CREEK 236.0
END DESCRIPTION:
XS GIS Cut Line= 2
      3729778.32     10765596.19      3727809.59     10765505.91
#Sta/Elev= 30
    4306  473.67  4334.7  471.27  4364.8  471.96  4404.8  469.19  4474.9  470.13
  4524.9  468.03    4555   462.7    4575   462.1  4685.1  449.29  4805.2  440.71
  4845.1  438.83  4944.1  436.38  4978.6  435.58  4981.4  435.08  4984.6  435.58
  5125.6  435.58  5235.7  438.71  5395.9  440.65    5516  444.73  5626.1  441.61
  5639.4  442.99  5846.3  443.96  5986.5   449.5    6073  458.68    6078  457.53
  6116.6  462.75  6136.6  466.99  6156.7  468.89  6196.7  469.71  6276.8  467.44
#Mann= 5 ,-1 , 0
    4306     .05       0  4845.1     .08       0  4944.1     .05       0
  4978.6     .04       0  4984.6     .05       0
Bank Sta=4805.2,5395.9
XS Rating Curve= 0 ,0
Exp/Cntr=0.3,0.1

Type RM Length L Ch R = 1 ,228153  ,582,582,582
BEGIN DESCRIPTION:
CATFISH CREEK 235.0
END DESCRIPTION:
XS GIS Cut Line= 2
      3729733.23     10765530.22      3727830.44     10765436.47
#Sta/Elev= 30
  4367.8  470.92  4441.5  464.96  4468.3   465.1  4531.6  460.87  4581.7  460.35
  4601.7  458.66  4631.7  452.69    4670  448.98  4781.9  441.39    4832  440.69
  4902.1  437.57  4942.1  437.91  4959.1  435.42  4961.9  434.92  4965.1  435.42
  5032.2  435.69  5052.2  438.04  5092.3  437.42  5162.4  440.91  5262.5   445.2
  5280.2  443.22  5302.6  445.87  5362.6  443.26  5522.8  444.35  5622.9  447.33
  5733.1  444.65  5913.3  445.76  6043.4  451.18  6223.7  466.96  6272.9  467.84
#Mann= 3 ,-1 , 0
  4367.8     .05       0  4959.1     .03       0  4965.1     .05       0
Bank Sta=4832,5162.4
XS Rating Curve= 0 ,0
Exp/Cntr=0.3,0.1

Type RM Length L Ch R = 1 ,227571  ,443,443,443
BEGIN DESCRIPTION:
CATFISH CREEK 234.0
END DESCRIPTION:
XS GIS Cut Line= 3
      3729599.57     10765160.17      3729299.61     10764960.19
      3728999.56     10764910.18
#Sta/Elev= 30
  4649.9  464.52  4685.9  461.15  4693.4  459.33  4699.4  458.78  4708.4  455.82
    4722  456.08  4735.5   454.7  4750.5  451.61  4765.5  449.61  4786.6  448.05
  4858.7   440.4  4908.7  436.49  4938.3  436.03  4966.8  436.83  4978.9  435.42
  4981.6  434.92  4984.9  435.42  5043.4  435.42    5047  436.13  5081.4  440.34
  5142.2  446.12  5172.6  449.59    5203  454.53  5213.2  454.88  5220.8     457
  5243.6  461.19    5274  465.34  5281.6  468.06  5286.7  468.23  5314.6  473.02
#Mann= 5 ,-1 , 0
  4649.9     .05       0  4908.7     .16       0  4978.9     .07       0
  4984.9     .16       0    5047     .05       0
Bank Sta=4858.7,5081.4
XS Rating Curve= 0 ,0
Exp/Cntr=0.3,0.1

Type RM Length L Ch R = 1 ,227128  ,413,413,413
BEGIN DESCRIPTION:
CATFISH CREEK 233.0
END DESCRIPTION:
XS GIS Cut Line= 3
      3729499.65     10764410.17      3729149.61     10764560.19
       3728899.6     10764660.19
#Sta/Elev= 30
  4650.8  471.83  4672.6   469.4  4712.5  458.35    4727  457.85  4741.5  456.52
  4748.8  453.45  4770.5  449.64  4781.4  448.91  4794.1  446.06  4803.2  445.52
  4812.2  443.89  4846.7  440.39  4857.6   438.6  4888.4  436.58  4890.8  435.42
  4893.6  434.92  4896.8  435.42  4998.4  435.42  5094.9  435.42  5100.3  437.43
    5107  438.51  5117.8   439.3  5124.5  440.51  5193.2  448.12  5202.6  450.68
  5256.5   458.4  5268.6  461.76  5279.4  462.77  5286.1  464.52  5300.9  466.12
#Mann= 5 ,-1 , 0
  4650.8     .05       0  4890.8     .07       0  4896.8     .05       0
  4998.4     .16       0    5107     .05       0
Bank Sta=4846.7,5124.5
XS Rating Curve= 0 ,0
Exp/Cntr=0.3,0.1

Type RM Length L Ch R = 1 ,226715  ,422,422,422
BEGIN DESCRIPTION:
CATFISH CREEK 232.0
END DESCRIPTION:
XS GIS Cut Line= 3
      3729399.65      10764260.2      3728999.61     10764160.19
      3728749.66     10764160.19
#Sta/Elev= 30
  4610.7  459.18  4633.9  458.56  4641.7  456.79  4662.3  453.72    4670  451.82
  4675.2  452.08  4711.2  447.39  4716.4  447.39  4744.7  444.35  4752.5  442.78
  4757.6  442.97  4765.4  441.16  4775.7  440.58  4806.6  436.93  4816.9  436.72
  4824.2  435.42    4827  434.92  4830.2  435.42  5124.6  435.61    5143  437.13
    5153     439    5163  439.78    5173   442.4    5183  443.27    5203  448.19
    5223  452.34    5233  453.78    5243  456.77    5263  460.03    5273  460.43
#Mann= 4 ,-1 , 0
  4610.7     .05       0  4824.2    .033       0  4830.2     .05       0
  5124.6     .16       0
Bank Sta=4775.7,5173
XS Rating Curve= 0 ,0
Exp/Cntr=0.3,0.1

Type RM Length L Ch R = 1 ,226293  ,416,416,416
BEGIN DESCRIPTION:
CATFISH CREEK 231.0
END DESCRIPTION:
XS GIS Cut Line= 3
      3729049.62     10763510.18      3728799.61     10763810.19
      3728699.59     10764110.24
#Sta/Elev= 30
  4616.2  468.35  4629.9  466.46  4644.2  466.36  4687.2  461.86  4758.7  451.23
  4772.4  449.88  4786.1  446.33  4793.9  446.54  4823.4  442.21    4829  440.95
  4836.8  440.69  4857.7  438.09  4864.2  435.51    4872  436.27  4875.5  435.42
  4878.3  434.92  4881.5  435.42  5154.3  435.42  5165.2  436.98  5175.4  437.62
  5185.9  439.79  5196.5  440.29  5217.5  443.85  5238.6  445.54  5270.2  449.78
  5280.8  452.09  5291.3  452.63  5301.9  454.76  5312.4  455.25    5323  456.96
#Mann= 5 ,-1 , 0
  4616.2     .16       0  4823.4     .05       0  4875.5    .033       0
  4881.5     .05       0  5165.2     .16       0
Bank Sta=4836.8,5185.9
XS Rating Curve= 0 ,0
Exp/Cntr=0.3,0.1

Type RM Length L Ch R = 1 ,225877  ,415,415,415
BEGIN DESCRIPTION:
CATFISH CREEK 230.0
END DESCRIPTION:
XS GIS Cut Line= 3
      3728949.65     10763410.18      3728549.61     10763460.19
      3728149.57     10763710.21
#Sta/Elev= 30
  4624.9  459.75  4655.2  454.69  4662.7  454.06  4667.8  455.02  4675.3  453.05
  4705.6  449.34  4715.6  447.11  4735.8   445.6  4743.4  444.01  4748.4  445.84
    4756  444.37    4766     444  4796.3  440.39  4803.6  439.24    4824  436.95
    4829   437.9  4843.7  435.42  4846.4  434.92  4849.7  435.42  5292.1  435.42
    5340  435.42    5370  440.12  5376.5  442.12  5413.1  446.54    5419  448.15
  5428.4  448.97  5434.3  450.77  5470.9  452.85  5476.8  454.84  5499.8  456.07
#Mann= 5 ,-1 , 0
  4624.9     .16       0  4803.6     .05       0  4843.7    .033       0
  4849.7     .05       0  5292.1     .16       0
Bank Sta=4796.3,5370
XS Rating Curve= 0 ,0
Exp/Cntr=0.3,0.1

Type RM Length L Ch R = 1 ,225462  ,427,427,427
BEGIN DESCRIPTION:
CATFISH CREEK 229.0
END DESCRIPTION:
XS GIS Cut Line= 3
      3728749.64     10763010.18      3728349.61     10763110.19
      3728149.57     10763210.21
#Sta/Elev= 30
  4584.5  462.75  4594.8     462  4602.6  460.12  4607.7   460.7  4615.5  459.84
  4636.1   456.3  4643.8  454.09  4677.3  449.34    4685  447.32  4690.2  447.43
  4697.9  446.42  4727.6  441.03  4739.2  439.87  4772.7  436.67  4777.4  435.42
  4780.1  434.92  4783.4  435.42  5122.6  435.42    5131  436.46  5139.4  439.17
    5145  439.74  5153.4  441.41  5157.3  443.34  5161.8  445.57  5167.3  446.81
  5175.7  447.45  5189.7  451.17  5198.1  451.89  5206.5  454.24  5220.5  455.46
#Mann= 5 ,-1 , 0
  4584.5     .16       0  4727.6     .05       0  4777.4    .033       0
  4783.4     .05       0  5157.3     .16       0
Bank Sta=4739.2,5145
XS Rating Curve= 0 ,0
Exp/Cntr=0.3,0.1

Type RM Length L Ch R = 1 ,225035  ,431,431,431
BEGIN DESCRIPTION:
CATFISH CREEK 228.0
END DESCRIPTION:
XS GIS Cut Line= 3
      3728499.57     10762710.19      3728099.61     10762760.19
       3727699.6     10762860.19
#Sta/Elev= 30
  4601.6  463.58  4611.6  463.41    4662  456.46  4672.1  455.69  4692.3  452.19
    4720  448.76    4725  448.66  4732.6  446.45  4742.7  445.78  4752.7  442.44
  4762.8   441.4  4775.2  439.12    4793  437.03  4797.6  435.42  4800.4  434.92
  4803.6  435.42  5192.8  435.42  5200.5  438.45  5210.8  439.38  5221.1   441.6
  5241.8   445.2  5250.9  445.57  5270.1  448.48    5283  452.11  5311.3  455.43
  5324.2  459.41  5334.5  460.22  5365.4  467.17  5385.5  468.65    5417  470.99
#Mann= 6 ,-1 , 0
  4601.6     .16       0  4775.2     .05       0  4797.6    .033       0
  4803.6     .05       0  5250.9     .16       0  5385.5     .05       0
Bank Sta=4762.8,5221.1
XS Rating Curve= 0 ,0
Exp/Cntr=0.3,0.1

Type RM Length L Ch R = 1 ,224604  ,477,477,477
BEGIN DESCRIPTION:
CATFISH CREEK 227.0
END DESCRIPTION:
XS GIS Cut Line= 3
      3728149.63     10762260.18      3727849.61     10762410.19
       3727599.6     10762660.19
#Sta/Elev= 30
  4676.1  453.74  4712.5  452.27  4729.2  450.82  4734.8  451.01  4751.6  449.21
  4757.2   449.3  4765.6  447.96  4787.9   446.3  4796.3  444.11  4801.9  444.03
  4810.3  443.05  4818.7  440.44  4824.3  440.52  4832.7  439.18    4841  435.61
  4843.6  435.42  4846.4  434.92  4849.6  435.42  5195.4  435.42  5209.5  437.24
  5223.7  438.35  5237.8  441.27    5252  443.82  5266.1  445.54  5280.2  448.98
  5294.4  450.36  5308.5  453.84  5336.8  459.76  5361.6  466.41  5365.1  466.41
#Mann= 3 ,-1 , 0
  4676.1     .05       0  4843.6    .033       0  4849.6     .05       0
Bank Sta=4824.3,5237.8
XS Rating Curve= 0 ,0
Exp/Cntr=0.3,0.1

Type RM Length L Ch R = 1 ,224127  ,441,441,441
BEGIN DESCRIPTION:
CATFISH CREEK 226.0
END DESCRIPTION:
XS GIS Cut Line= 3
      3727899.63     10761710.17      3727499.61     10762110.19
      3727099.62     10762410.18
#Sta/Elev= 30
  4410.5  465.78  4414.1  465.78  4438.8  461.79    4453  457.67  4537.8  446.47
  4608.5  443.26  4636.8  444.75  4650.9  446.52  4693.4  447.67  4735.8  443.09
  4749.9  440.42  4761.1  435.42  4763.8  434.92  4767.1  435.42  5218.9  435.42
  5233.5  438.62  5248.1  439.61  5254.3  441.96  5262.7  442.52  5276.2  445.39
  5289.8  446.82  5304.3  450.12  5312.7  450.92  5326.2  455.95  5348.1   461.5
  5368.9   464.3  5398.1  466.34  5418.9  469.09  5448.1  470.68  5476.2  474.13
#Mann= 3 ,-1 , 0
  4410.5     .05       0  4761.1    .033       0  4767.1     .05       0
Bank Sta=4749.9,5254.3
XS Rating Curve= 0 ,0
Exp/Cntr=0.3,0.1

Type RM Length L Ch R = 1 ,223686  ,423,423,423
BEGIN DESCRIPTION:
CATFISH CREEK 225.0
END DESCRIPTION:
XS GIS Cut Line= 3
      3727499.57     10761610.22      3727099.61     10761910.19
      3726949.59     10762310.23
#Sta/Elev= 30
  4503.5  454.82  4510.7  453.99  4531.6  456.02  4539.9  455.08  4546.2  456.36
  4560.7  453.79    4567  454.05    4617  449.82  4625.3  447.99  4639.9  447.53
    4667  449.11  4675.3   443.2  4681.6  443.87  4689.9  440.79  4696.2  438.63
  4703.5  438.26    4714  435.42  4716.7  434.92    4720  435.42  5164.5  435.42
  5174.3  437.86  5189.5   439.3  5195.7  441.52  5206.4  443.32  5214.4  445.98
    5250  450.23  5259.8  452.99  5269.6  454.06  5291.8  458.69  5430.7  474.17
#Mann= 3 ,-1 , 0
  4503.5     .05       0    4714    .033       0    4720     .05       0
Bank Sta=4689.9,5195.7
XS Rating Curve= 0 ,0
Exp/Cntr=0.3,0.1

Type RM Length L Ch R = 1 ,223263  ,428,428,428
BEGIN DESCRIPTION:
CATFISH CREEK 224.0
END DESCRIPTION:
XS GIS Cut Line= 3
      3726549.61     10760960.19      3726699.61     10761760.19
      3726699.61     10762160.15
#Sta/Elev= 30
  4157.4  488.93  4167.6  488.77  4228.6  484.03    4249  481.38  4288.8  478.23
  4299.8  475.93  4330.4  472.65  4351.6  467.23  4421.9  457.24  4493.1  449.69
  4509.3   446.9  4561.8  440.39  4566.9  440.77  4574.5  439.82  4584.7  438.38
  4619.5  436.88  4625.4  435.55  4632.6  435.42  4635.3  434.92  4638.6  435.42
  5171.3  435.42  5181.3     439  5191.3  439.72  5201.3   442.5  5211.3  443.58
  5221.3  446.25  5231.3  447.05  5261.3  452.06  5271.3   452.6  5371.3  464.04
#Mann= 3 ,-1 , 0
  4157.4     .05       0  4632.6    .033       0  4638.6     .05       0
Bank Sta=4574.5,5191.3
XS Rating Curve= 0 ,0
Exp/Cntr=0.3,0.1

Type RM Length L Ch R = 1 ,222835  ,209,209,209
BEGIN DESCRIPTION:
CATFISH CREEK 223.0
END DESCRIPTION:
XS GIS Cut Line= 3
      3726366.65     10761185.62      3726271.16     10761767.26
      3726400.94     10762346.98
#Sta/Elev= 30
  4492.5  464.88  4497.4  464.88  4517.4  461.44  4547.8  459.03  4578.2  455.33
  4626.2  453.83    4639  452.42  4659.3  449.68  4669.4  446.82  4699.8   441.2
  4709.9  438.99  4748.7  435.45  4757.6  435.42  4760.4  434.92  4763.6  435.42
  5361.6  435.42  5369.6  438.46  5392.4  440.22  5402.6  442.83  5418.1  444.61
  5423.2  447.06  5433.3  449.21  5461.4  451.99  5466.6  454.86  5474.3  456.24
  5504.8  456.88  5515.3  460.23  5576.8  465.02  5628.1  467.78    5676  472.19
#Mann= 3 ,-1 , 0
  4492.5     .05       0  4757.6    .033       0  4763.6     .05       0
Bank Sta=4699.8,5392.4
XS Rating Curve= 0 ,0
Exp/Cntr=0.3,0.1

Type RM Length L Ch R = 1 ,222626  ,60,60,60
BEGIN DESCRIPTION:
CATFISH CREEK 222.0
END DESCRIPTION:
XS GIS Cut Line= 2
      3726192.03     10761085.49      3725910.92     10762485.85
#Sta/Elev= 30
  4445.1  460.46    4530  453.56  4643.7  440.56  4682.7  436.72  4745.7  437.01
  4763.1  435.42  4765.8  434.92  4769.1  435.42  4898.7  436.57  4937.2  435.42
  4942.3  436.59  5242.6  435.42  5265.9  436.65  5293.6  435.42  5298.7  436.75
  5344.5  435.42  5349.6  437.06  5395.4  437.49  5400.5  438.99  5497.2  439.52
  5502.3  440.92  5553.2  440.32    5599  436.93  5663.6  436.14  5714.6  437.35
    5735  439.75  5751.7   442.9  5756.8   441.6  5847.2  451.13  5873.4  458.09
#Mann= 3 ,-1 , 0
  4445.1     .05       0  4763.1     .03       0  4769.1     .05       0
Bank Sta=4643.7,5735
XS Rating Curve= 0 ,0
Exp/Cntr=0.3,0.1

Type RM Length L Ch R = 1 ,222566  ,157,157,157
BEGIN DESCRIPTION:
Mapping XS c79cb669
END DESCRIPTION:
XS GIS Cut Line= 3
        3726128.     10761120.09      3725917.06     10762133.14
      3725838.93     10762539.42
#Sta/Elev= 30
  4496.2  452.76  4526.9  449.75  4612.4  447.19  5292.8  446.91  5297.9  443.35
  5303.2  445.29  5342.9  446.17    5348  442.31  5354.3  444.72    5393  446.02
  5398.1  442.19  5405.4  444.66  5425.8  445.59    5443   446.2  5448.1  443.92
  5517.7  447.04  5543.6  441.73  5652.6  440.89  5670.5   438.5  5696.4  435.38
  5699.2  434.88  5702.4  435.38  5772.4  438.01  5782.6  441.43  5833.5  443.92
  5853.8  446.27  5860.3  448.96  5865.4  447.19  5904.8  457.16  5944.7  457.49
#Mann= 3 ,-1 , 0
  4496.2     .05       0  5696.4     .03       0  5702.4     .05       0
Bank Sta=5670.5,5772.4
XS Rating Curve= 0 ,0
Exp/Cntr=0.3,0.1

Type RM Length L Ch R = 1 ,222409  ,461,461,461
BEGIN DESCRIPTION:
Mapping XS 42ef63d8
END DESCRIPTION:
XS GIS Cut Line= 2
      3726014.95     10761033.42      3725718.55     10762167.01
#Sta/Elev= 30
  4444.6  461.31  4564.7  446.66  4643.2   439.1  4683.6  437.07  4759.3  428.01
  4764.5  428.97  4798.8  423.46    4805  424.58  4840.2  420.19  4885.8  417.57
  4915.6  412.86  4937.4  409.97  4989.1  409.79  5118.1  407.61  5193.8  409.51
    5196  407.59  5198.7  407.09    5202  407.59  5206.1  409.19  5226.8   408.5
  5257.8  411.48  5299.2  411.66  5361.2  417.13  5390.9  422.37    5396  421.06
  5426.8  425.02  5471.7  428.59  5586.3  431.95  5598.9  433.07  5616.3  439.89
#Mann= 8 ,-1 , 0
  4444.6     .16       0  4564.7     .05       0  4798.8     .16       0
  4915.6     .05       0    5196     .03       0    5202     .05       0
  5426.8     .16       0  5586.3     .05       0
Bank Sta=4989.1,5257.8
XS Rating Curve= 0 ,0
Exp/Cntr=0.3,0.1

Type RM Length L Ch R = 1 ,221948  ,476,476,476
BEGIN DESCRIPTION:
CATFISH CREEK 221.0
END DESCRIPTION:
XS GIS Cut Line= 3
      3725359.08     10760938.94      3725449.61     10761510.19
      3725478.88     10762074.35
#Sta/Elev= 30
  4411.1  448.79  4422.5   448.8  4432.6  447.18  4447.1  446.87  4473.1  443.41
  4594.6  431.71    4625  431.38  4646.9   428.5  4706.5   422.7  4736.4  418.62
  4768.8  416.44  4817.4  411.37  4893.5  406.69  4918.6  406.47  4980.5   405.1
  5009.5  402.99  5019.5  404.86  5029.5  405.11  5046.6  401.79  5049.3  401.29
  5052.6  401.79  5059.6   402.1  5069.6  404.82    5163  404.12  5259.8  403.85
  5289.9  406.36  5473.6  423.08  5500.7  427.24    5504  427.38  5554.4  432.82
#Mann= 8 ,-1 , 0
  4411.1     .12       0  4646.9     .05       0  4980.5     .16       0
  5046.6     .07       0  5052.6     .16       0    5163     .05       0
  5500.7     .16       0    5504     .05       0
Bank Sta=4918.6,5289.9
XS Rating Curve= 0 ,0
Exp/Cntr=0.3,0.1

Type RM Length L Ch R = 1 ,221472  ,657,657,657
BEGIN DESCRIPTION:
CATFISH CREEK 220.0
END DESCRIPTION:
XS GIS Cut Line= 3
      3724949.61     10761210.17      3724999.61     10761610.19
      3725299.59     10762010.17
#Sta/Elev= 30
  4648.5  432.66  4675.8  428.24  4686.3  424.97    4709  420.94  4759.4  414.91
  4779.5  414.59  4799.7  412.12  4920.6  403.79    4969  402.51    4971  402.58
  4981.1  401.51  4998.2  396.91    5001  396.41  5004.2  396.91  5008.8  401.18
  5013.8  402.35  5021.4  402.09  5041.5  397.26  5054.8  398.82  5058.9  402.19
  5179.8  401.02    5267  401.73  5279.8  401.69  5338.1  407.65  5344.3  406.87
  5423.5  416.48  5479.8  419.99  5508.9  423.74  5529.8  424.87  5551.6  428.55
#Mann= 6 ,-1 , 0
  4648.5     .12       0  4675.8     .05       0    4969     .16       0
  4998.2     .07       0  5004.2     .16       0    5267     .05       0
Bank Sta=4971,5058.9
XS Rating Curve= 0 ,0
Exp/Cntr=0.3,0.1

Type RM Length L Ch R = 1 ,220815  ,321,321,321
BEGIN DESCRIPTION:
CATFISH CREEK 219.0
END DESCRIPTION:
XS GIS Cut Line= 3
      3724849.61     10761160.19      3724699.61     10761410.19
      3724349.59     10761960.21
#Sta/Elev= 30
  4714.5  435.96  4772.8  430.09  4780.6  426.41  4796.1  424.12  4807.8  418.57
  4817.5  415.77  4838.9  412.09  4897.2  404.71  4955.5  399.75  4961.3  398.06
  4971.1  398.16  4982.7  394.93  4989.4   394.9  4992.2   394.4  4995.4   394.9
  4998.3  395.36  5003.1  398.37    5009  398.37  5013.7   399.9  5050.1  400.76
  5294.9  400.44  5321.6   400.4  5475.4  401.15  5500.5   401.6  5541.1   402.4
  5550.4  407.15  5556.4  407.34  5571.6  412.03  5588.8  413.99    5658  421.45
#Mann= 8 ,-1 , 0
  4714.5     .12       0  4989.4     .07       0  4995.4     .12       0
  5294.9     .16       0  5321.6     .12       0  5475.4     .16       0
  5500.5     .12       0  5588.8     .05       0
Bank Sta=4955.5,5013.7
XS Rating Curve= 0 ,0
Exp/Cntr=0.3,0.1

Type RM Length L Ch R = 1 ,220494  ,803,803,803
BEGIN DESCRIPTION:
CATFISH CREEK 218.0
END DESCRIPTION:
XS GIS Cut Line= 3
      3724711.55     10760787.79      3724383.43     10761334.65
      3723680.29     10761740.91
#Sta/Elev= 30
  4442.1  441.84  4548.4  430.17  4619.8   425.7  4692.2  417.95  4723.3  416.94
  4750.5  413.88  4861.3  407.25  4934.7  400.94  4956.6   400.5  4962.4  397.66
  4969.7   398.9  4977.9  398.06  4983.8  393.72    4990  393.25  4992.8  392.75
    4996  393.25  5014.9  399.57  5277.8  397.27  5582.2  398.01  5679.8  406.64
  5699.1   407.1  5754.1  411.99  5760.2  413.78  5781.8  413.43  5819.1  418.53
  5856.4  421.37  5862.2  420.62  5877.9  422.85  5883.7  421.43  5891.9   423.3
#Mann= 5 ,-1 , 0
  4442.1     .12       0    4990     .07       0    4996     .12       0
  5582.2     .16       0  5699.1     .05       0
Bank Sta=4969.7,5014.9
XS Rating Curve= 0 ,0
Exp/Cntr=0.3,0.1

Type RM Length L Ch R = 1 ,219691  ,1322,1322,1322
BEGIN DESCRIPTION:
CATFISH CREEK 217.0
END DESCRIPTION:
XS GIS Cut Line= 3
       3724249.6      10760810.2      3723899.61     10761210.19
      3723599.59     10761560.21
#Sta/Elev= 30
    4451  422.32  4585.3  408.96    4628  403.99  4635.6  402.25  4684.9   397.8
  4724.6  396.69  4839.4  397.56  4968.7  398.11  4985.8  397.25  4989.6  395.66
  4993.2  391.26    4996  390.76  4999.2  391.26  5003.9  391.28  5010.5  397.68
  5018.2  398.18  5024.7  396.74  5053.3  396.86  5081.8  395.58  5090.5  396.87
  5153.2  398.35  5215.5  404.06  5301.3  412.55  5351.3  419.04  5358.4  418.79
  5372.7  421.42  5422.1   427.2  5436.3  427.95  5440.2  429.53  5443.5  429.53
#Mann= 7 ,-1 , 0
    4451     .12       0  4724.6     .16       0  4839.4     .12       0
  4993.2     .07       0  4999.2     .12       0  5090.5     .16       0
  5215.5     .05       0
Bank Sta=4985.8,5010.5
XS Rating Curve= 0 ,0
Exp/Cntr=0.3,0.1

Type RM Length L Ch R = 1 ,218369  ,561,561,561
BEGIN DESCRIPTION:
CATFISH CREEK 215.0
END DESCRIPTION:
XS GIS Cut Line= 3
      3723599.62     10760360.18      3723299.61     10760710.19
       3722899.6     10761010.19
#Sta/Elev= 30
  4533.6  432.92  4604.4  425.83  4612.1  424.25  4625.8  417.87  4632.9  419.09
  4639.5  417.16  4661.5  415.66  4668.1  413.46    4690   410.4  4704.3  408.99
  4710.9  410.36  4725.1  406.83  4762.1  404.39  4803.1  399.01    4815  399.35
  4852.5  396.52  4916.1  394.88  4952.3  392.11  4958.9   393.8  4966.6  392.42
  4973.2  393.22  4998.9  389.85  5001.6  389.35  5004.9  389.85  5022.7  395.37
  5166.5  394.72  5251.9  396.39  5344.6   402.1    5381   406.9  5494.6  417.21
#Mann= 5 ,-1 , 0
  4533.6     .16       0  4762.1     .12       0    4815     .16       0
  4998.9     .07       0  5004.9     .16       0
Bank Sta=4916.1,5022.7
XS Rating Curve= 0 ,0
Exp/Cntr=0.3,0.1

Type RM Length L Ch R = 1 ,217808  ,417,417,417
BEGIN DESCRIPTION:
CATFISH CREEK 214.0
END DESCRIPTION:
XS GIS Cut Line= 2
      3723245.43     10760081.15      3722654.45     10760830.94
#Sta/Elev= 30
  4522.2  426.19  4533.5  424.28  4554.3  423.77  4574.8   421.8  4658.5  414.82
  4732.3  408.19  4796.4  400.05  4839.3  397.49  4846.1  396.15  4916.7  392.85
  4966.6  393.58  4980.8  392.81  4988.9  387.25  4992.2  387.11    4995  386.61
  4998.2  387.11  5003.3  387.94  5009.7  392.68  5017.6  393.73  5158.8  392.92
  5259.5  396.87  5315.1  401.19  5351.2  403.32  5380.1  408.74  5386.8  408.66
  5400.9   412.5  5415.3  413.68  5429.8  417.45  5473.1  422.02  5476.9  423.38
#Mann= 6 ,-1 , 0
  4522.2     .12       0  4574.8     .16       0  4658.5     .12       0
  4992.2     .07       0  4998.2     .12       0  5315.1     .16       0
Bank Sta=4966.6,5017.6
XS Rating Curve= 0 ,0
Exp/Cntr=0.3,0.1

Type RM Length L Ch R = 1 ,217391  ,529,529,529
BEGIN DESCRIPTION:
CATFISH CREEK 213.0
END DESCRIPTION:
XS GIS Cut Line= 3
      3722849.62     10759960.17      3722649.61     10760360.19
       3722549.6     10760760.24
#Sta/Elev= 30
    4597  414.25  4627.8   410.1  4641.7  409.38  4686.5  404.52  4753.6  400.41
    4834  397.09  4924.1  393.65  4977.2  393.05  4985.5  391.88  4988.1  387.64
  4990.9  387.14  4994.1  387.64  4999.5  387.97  5007.9  390.81  5030.3   392.4
  5095.8  393.02  5116.4  392.09    5137  392.85  5149.9  394.78  5167.9  395.84
  5178.2  395.59  5219.5  398.94  5322.5  410.31  5332.9   410.4  5350.9  412.64
  5363.8   415.6  5374.1  415.86  5426.4  421.38  5433.4  422.79  5456.6  424.92
#Mann= 5 ,-1 , 0
    4597     .16       0    4834     .12       0  4988.1     .07       0
  4994.1     .12       0  5426.4     .16       0
Bank Sta=4977.2,5030.3
XS Rating Curve= 0 ,0
Exp/Cntr=0.3,0.1

Type RM Length L Ch R = 1 ,216862  ,733,733,733
BEGIN DESCRIPTION:
CATFISH CREEK 212.0
END DESCRIPTION:
XS GIS Cut Line= 3
      3722449.62     10759710.17      3722299.61     10760110.19
      3722324.21     10760720.17
#Sta/Elev= 30
  4531.2  429.28  4571.3   424.9  4576.6  425.59  4601.5  421.31  4606.9  422.37
  4616.7  420.06  4631.8  419.44  4662.1  414.35  4808.9  397.39    4905  391.17
  4943.3   390.1  4968.4  391.76  4998.5  385.53  5005.5  385.34  5008.2  384.84
  5011.5  385.34  5018.5  391.65  5048.5  391.89    5083  390.19  5188.6  391.39
    5232  393.27  5258.7  394.11  5318.7  399.37  5358.7  403.42  5375.9  407.17
  5438.8  414.73  5448.8  417.44  5518.9  425.43  5538.9  427.17  5568.9  427.35
#Mann= 5 ,-1 , 0
  4531.2     .12       0  5005.5     .07       0  5011.5     .12       0
    5232     .16       0  5375.9     .12       0
Bank Sta=4968.4,5018.5
XS Rating Curve= 0 ,0
Exp/Cntr=0.3,0.1

Type RM Length L Ch R = 1 ,216129  ,300,300,300
BEGIN DESCRIPTION:
CATFISH CREEK 211.0
END DESCRIPTION:
XS GIS Cut Line= 4
      3722412.02     10759542.98      3722030.09     10759633.26
      3721925.92     10759744.37      3721800.93     10760702.69
#Sta/Elev= 30
  4535.9  428.22  4743.9  414.16  4850.8  402.14    4926  391.07    4962  390.06
    4983  387.34  4990.3  388.81  4997.2   385.4  5008.4  384.65  5011.1  384.15
  5014.4  384.65  5018.7  389.27  5025.5  389.67  5080.7  388.97  5096.6  385.75
  5106.7  386.23  5116.8  389.27  5157.1   390.1  5197.5  389.08  5249.2  391.02
  5278.1   389.9  5555.1   392.6  5792.5  397.39    5853  399.96  5933.6  406.44
    5970  412.98  5994.2  418.37  6004.2   418.3    6019  421.94  6047.1  422.74
#Mann= 4 ,-1 , 0
  4535.9     .12       0  5008.4     .07       0  5014.4     .12       0
    5970     .16       0
Bank Sta=4962,5025.5
XS Rating Curve= 0 ,0
Exp/Cntr=0.3,0.1

Type RM Length L Ch R = 1 ,215829  ,698,698,698
BEGIN DESCRIPTION:
CATFISH CREEK 210.0
END DESCRIPTION:
XS GIS Cut Line= 3
       3722299.6      10759010.2      3721899.61     10759410.19
      3721149.63     10759960.18
#Sta/Elev= 30
  4400.9  444.28  4471.6  432.28  4499.9  425.28    4514  424.14  4598.9  411.01
  4669.6  401.74    4712  397.72  4768.6  395.66  4853.4  394.45  4938.3  389.54
  4994.8  389.11  5006.4  384.66  5009.2  384.16  5012.4  384.66  5016.2  387.63
  5024.1  389.64  5044.9  388.43  5095.1  389.87  5150.6  388.68  5193.5  388.15
  5295.8   389.6  5517.3  390.35  5552.8  391.66  5623.8  398.19  5655.9  400.03
  5688.6  402.29  5697.1  405.87  5782.2  417.02  5832.9  421.11  5896.6  423.65
#Mann= 7 ,-1 , 0
  4400.9     .12       0  5006.4     .07       0  5012.4     .12       0
  5150.6     .16       0  5193.5     .05       0  5655.9     .16       0
  5782.2     .12       0
Bank Sta=4994.8,5024.1
XS Rating Curve= 0 ,0
Exp/Cntr=0.3,0.1
