--- MILL BRANCH.prj (project) ---

Proj Title=MILL BRANCH Base Level Engineering
Current Plan=p01
Default Exp/Contr=0.3,0.1
English Units
Geom File=g01
Flow File=f01
Plan File=p01
Y Axis Title=Elevation
X Axis Title(PF)=Main Channel Distance
X Axis Title(XS)=Station
BEGIN DESCRIPTION:
MILL BRANCH
END DESCRIPTION:
DSS Export Rating Curves= 0
DSS Export Rating Curve Sorted= 0
DSS Export Volume Flow Curves= 0
DXF OffsetX= 0
DXF OffsetY= 0
DXF ScaleX= 1
DXF ScaleY= 10

--- MILL BRANCH.p01 (plan) ---

Plan Title=Multiple Run
Short Identifier=Multiple
Geom File=g01
Flow File=f01
Subcritical Flow
K Sum by GR= 0
Std Step Tol= 0.01
Critical Tol= 0.01
Num of Std Step Trials= 20
Max Error Tol= 0.3
Flow Tol Ratio= 0.001
Split Flow NTrial= 30
Split Flow Tol= 0.02
Split Flow Ratio= 0.02
Log Output Level= 0
Friction Slope Method= 1
Unsteady Friction Slope Method= 2
Unsteady Bridges Friction Slope Method= 1
Parabolic Critical Depth
Global Vel Dist=  1 , 1 , 1
Global Log Level= 0
CheckData=True
Encroach Param= -1, 0, 0, 0
BEGIN DESCRIPTION:
Multiple Run
END DESCRIPTION:

--- MILL BRANCH.f01 (steady flow) ---

Flow Title=Multiple
Program Version=4.10
Number of Profiles= 7
Profile Names=10-year,25-year,50-year,1pct_min,100-year,1pct_plu,500-year
River Rch & RM=MILL BRANCH,Reach-1         ,43139
     465     622     750     664     898    1214    1289
River Rch & RM=MILL BRANCH,Reach-1         ,42081
     770    1061    1304    1175    1589    2150    2367
River Rch & RM=MILL BRANCH,Reach-1         ,40828
     819    1128    1387    1249    1689    2284    2511
River Rch & RM=MILL BRANCH,Reach-1         ,38429
    1203    1691    2105    1918    2594    3508    3952
River Rch & RM=MILL BRANCH,Reach-1         ,35202
    1470    2084    2610    2391    3234    4374    4979
River Rch & RM=MILL BRANCH,Reach-1         ,32423
    1495    2120    2655    2432    3289    4448    5063
River Rch & RM=MILL BRANCH,Reach-1         ,29994
    2268    3275    4153    3846    5202    7035    8189
River Rch & RM=MILL BRANCH,Reach-1         ,29091
    2778    4034    5134    4769    6449    8722   10212
River Rch & RM=MILL BRANCH,Reach-1         ,28255
    2778    4034    5134    4769    6449    8722   10212
River Rch & RM=MILL BRANCH,Reach-1         ,25264
    2878    4173    5306    4922    6657    9002   10513
River Rch & RM=MILL BRANCH,Reach-1         ,20034
    2891    4184    5312    4921    6654    8999   10476
River Rch & RM=MILL BRANCH,Reach-1         ,18810
    2891    4184    5312    4921    6654    8999   10476
River Rch & RM=MILL BRANCH,Reach-1         ,16248
    3602    5254    6707    6242    8442   11417   13420
River Rch & RM=MILL BRANCH,Reach-1         ,15685
    4024    5886    7528    7018    9491   12835   15134
River Rch & RM=MILL BRANCH,Reach-1         ,14449
    4024    5886    7528    7018    9491   12835   15134
River Rch & RM=MILL BRANCH,Reach-1         ,9257
    4326    6335    8107    7562   10227   13830   16323
River Rch & RM=MILL BRANCH,Reach-1         ,8722
    4326    6335    8107    7562   10227   13830   16323
River Rch & RM=MILL BRANCH,Reach-1         ,4799
    4362    6379    8157    7600   10278   13899   16368
River Rch & RM=MILL BRANCH,Reach-1         ,2000
    4381    6402    8181    7618   10302   13933   16388
Boundary for River Rch & Prof#=MILL BRANCH,Reach-1         , 1
Up Type= 0
Dn Type= 3
Dn Slope=0.00239
Boundary for River Rch & Prof#=MILL BRANCH,Reach-1         , 2
Up Type= 0
Dn Type= 3
Dn Slope=0.00239
Boundary for River Rch & Prof#=MILL BRANCH,Reach-1         , 3
Up Type= 0
Dn Type= 3
Dn Slope=0.00239
Boundary for River Rch & Prof#=MILL BRANCH,Reach-1         , 4
Up Type= 0
Dn Type= 3
Dn Slope=0.00239
Boundary for River Rch & Prof#=MILL BRANCH,Reach-1         , 5
Up Type= 0
Dn Type= 3
Dn Slope=0.00239
Boundary for River Rch & Prof#=MILL BRANCH,Reach-1         , 6
Up Type= 0
Dn Type= 3
Dn Slope=0.00239
Boundary for River Rch & Prof#=MILL BRANCH,Reach-1         , 7
Up Type= 0
Dn Type= 3
Dn Slope=0.00239
DSS Import GetInterval= 0
DSS Import GetPeak= 0
DSS Import FillOption= 0

--- MILL BRANCH.g01 (geometry) ---

Geom Title=Existing Conditions
Program Version=4.10

River Reach=MILL BRANCH     ,Reach-1
Reach XY= 30
      3675869.63     10781197.61      3675060.75       10780755.
        3675153.       10779583.       3674725.5       10777501.
      3675047.75       10776606.      3674435.75       10774181.
       3675964.5       10771029.       3676155.5       10769930.
        3675935.       10769477.      3676023.25       10768113.
        3676335.       10767938.      3676556.25       10767224.
      3676091.25       10765078.       3676472.5       10762507.
       3677732.5       10761221.      3678109.25       10760460.
      3678950.25       10760004.        3679185.       10759528.
       3680409.5       10758530.        3681961.       10757807.
      3682433.25       10757294.      3682369.75       10756164.
      3682783.75       10755483.        3682870.       10754247.
        3686020.       10751676.      3685986.75       10751324.
        3686628.       10750135.       3688354.5       10749015.
       3689081.5       10749341.       3689559.5       10748921.

Type RM Length L Ch R = 1 ,43139   ,483,483,483
BEGIN DESCRIPTION:
MILL BRANCH 78.0
END DESCRIPTION:
XS GIS Cut Line= 3
      3675949.62     10780960.18      3675749.61     10781160.19
      3675699.59     10781260.23
#Sta/Elev= 30
  4731.3  456.09  4745.5  455.45  4759.6  454.07  4773.7  453.63  4787.9  451.42
    4802  450.47  4816.2  447.21  4858.6  441.47  4886.9   436.7    4901  434.75
  4915.2  433.54  4957.6  432.71  4971.7  432.94  4985.9  432.16    4997   429.9
  4999.8   429.4    5003   429.9  5010.6  432.92  5016.9  432.92  5022.5  434.19
  5036.5  435.99  5044.9  438.03  5058.9  439.21  5067.3  441.09  5072.8  441.42
  5089.6  444.37  5103.6   447.5  5117.6  449.24  5123.2  451.42    5126  451.42
#Mann= 3 ,-1 , 0
  4731.3     .12       0    4997     .07       0    5003     .12       0
Bank Sta=4886.9,5036.5
XS Rating Curve= 0 ,0
Exp/Cntr=0.3,0.1

Type RM Length L Ch R = 1 ,42656   ,166,166,166
BEGIN DESCRIPTION:
MILL BRANCH 77.0
END DESCRIPTION:
XS GIS Cut Line= 3
      3675449.62     10780760.15      3675399.61     10780910.19
      3675449.61     10781210.19
#Sta/Elev= 30
  4845.1  446.18  4887.3  441.94  4897.8  440.06  4918.9   437.6  4929.5   435.1
    4940  434.08  4950.6  432.21  4961.1  430.98  4971.6  430.93  4992.7  428.99
  5005.8   429.5  5028.1  428.66  5030.9  428.16  5034.1  428.66  5036.2  429.38
  5053.9  429.12    5092  430.68  5135.1  430.76  5145.5  429.17  5152.8  429.51
  5165.5   431.2  5175.6  431.83  5185.7  434.67  5195.9   435.1  5226.3  439.82
  5246.6  441.09  5256.7  441.22  5276.3  443.14  5287.1  444.42  5307.4  445.89
#Mann= 5 ,-1 , 0
  4845.1     .16       0  5028.1     .07       0  5034.1     .16       0
  5145.5     .12       0  5276.3     .16       0
Bank Sta=4971.6,5092
XS Rating Curve= 0 ,0
Exp/Cntr=0.3,0.1

Type RM Length L Ch R = 1 ,42490   ,409,409,409
BEGIN DESCRIPTION:
Mapping XS 7e976db1
END DESCRIPTION:
XS GIS Cut Line= 2
      3675430.34      10780667.6      3675008.44     10781224.92
#Sta/Elev= 30
  4705.3  450.94  4731.3  449.63  4779.3  446.76  4829.2  440.34  4835.5  441.19
  4864.6  438.81  4879.2  435.47  4885.4  436.77  4893.7  433.21  4908.3  430.71
  4935.4  428.55  4954.4  428.46  4971.9  428.11    4979  426.14  4996.9  423.85
  4999.6  423.35  5002.9  423.85  5008.2  426.15  5022.1   427.7    5029  427.03
  5035.3  428.34  5075.8  430.25  5099.7  430.97    5115   432.7    5158  438.37
  5172.5  441.47  5193.3  442.62  5199.6  443.99  5328.4  447.69  5404.3  448.23
#Mann= 8 ,-1 , 0
  4705.3     .05       0  4731.3     .16       0  4954.4     .12       0
  4996.9     .07       0  5002.9     .12       0  5075.8     .16       0
    5115     .05       0  5328.4     .16       0
Bank Sta=4971.9,5022.1
XS Rating Curve= 0 ,0
Exp/Cntr=0.3,0.1

Type RM Length L Ch R = 1 ,42081   ,309,309,309
BEGIN DESCRIPTION:
Mapping XS 45b13d4b
END DESCRIPTION:
XS GIS Cut Line= 3
      3675487.66     10780571.24       3675034.5      10780667.6
      3674560.57     10780654.58
#Sta/Elev= 30
    4611  454.42    4701  451.75  4731.7  449.39  4782.8   448.9    4806  446.93
  4833.9  443.18  4854.4   441.7  4864.6  442.42    4870  439.43  4908.1  434.14
  4946.4  428.15  4969.2  425.11  4987.3  424.77  4994.5  422.33  4997.3  421.83
  5000.5  422.33  5010.2  424.25  5028.2   425.5  5079.2  424.72  5119.2  427.83
    5131  430.23  5158.2   434.9  5163.2  433.69  5189.2   435.9  5199.2  437.15
  5209.2  440.02  5239.2  442.55  5335.8  445.34  5451.6  450.53  5548.4  454.43
#Mann= 9 ,-1 , 0
    4611     .05       0    4806     .12       0  4908.1     .16       0
  4994.5     .07       0  5000.5     .16       0  5010.2     .12       0
    5131     .16       0  5335.8     .12       0  5451.6     .16       0
Bank Sta=4946.4,5119.2
XS Rating Curve= 0 ,0
Exp/Cntr=0.3,0.1

Type RM Length L Ch R = 1 ,41772   ,400,400,400
BEGIN DESCRIPTION:
MILL BRANCH 76.0
END DESCRIPTION:
XS GIS Cut Line= 2
      3675508.13     10780410.95      3674523.78     10780367.59
#Sta/Elev= 30
    4514  456.33  4632.6  453.32  4652.7  451.53  4682.7  451.91  4717.3  447.58
  4762.8  443.45  4772.8  441.56  4782.8  438.25  4816.2  434.32  4852.8  428.34
  4892.9  422.58  4915.2  422.66  4932.9  422.51  4952.9  423.82    5000  422.05
  5002.7  421.55    5006  422.05  5061.7  426.94  5083.1  428.92  5098.7  431.88
  5133.1  436.42  5143.1  439.41  5183.2  444.65  5213.2  447.58  5253.2  448.42
  5303.3  451.54  5463.4   457.2  5473.4  458.18  5493.5  458.59  5499.3   459.6
#Mann= 7 ,-1 , 0
    4514     .05       0  4717.3     .12       0  4816.2     .16       0
  4915.2     .12       0    5000     .07       0    5006     .12       0
  5061.7     .16       0
Bank Sta=4852.8,5061.7
XS Rating Curve= 0 ,0
Exp/Cntr=0.3,0.1

Type RM Length L Ch R = 1 ,41372   ,372,372,372
BEGIN DESCRIPTION:
MILL BRANCH 75.0
END DESCRIPTION:
XS GIS Cut Line= 2
      3675555.81     10780024.66      3674303.02     10779976.98
#Sta/Elev= 30
  4545.8   454.8  4642.1  452.73  4762.2  447.08  4782.2   444.9    4796  441.94
  4810.2  440.13  4852.2  434.62  4862.2  432.12  4892.3  427.62  4902.3  425.36
  4912.3  424.78  4922.3  422.87  4952.3  420.79  5029.4  420.69  5032.1  420.19
  5035.4  420.69  5052.4  421.83  5078.6  425.24  5082.4   425.7  5132.4  432.84
  5177.5  438.24  5202.5     442  5222.5  446.82  5232.5  447.81  5312.6  449.81
  5609.1  461.43  5662.8  463.02  5692.8  465.45  5771.1  469.04  5799.5  470.59
#Mann= 8 ,-1 , 0
  4545.8     .05       0  4810.2     .16       0  5029.4     .07       0
  5035.4     .16       0  5078.6     .12       0  5177.5     .16       0
  5609.1     .07       0  5771.1     .05       0
Bank Sta=4892.3,5082.4
XS Rating Curve= 0 ,0
Exp/Cntr=0.3,0.1

Type RM Length L Ch R = 1 ,41000   ,172,172,172
BEGIN DESCRIPTION:
MILL BRANCH 74.0
END DESCRIPTION:
XS GIS Cut Line= 4
      3675816.24     10779655.74      3675321.47      10779651.4
      3674896.12     10779720.84      3674006.37     10779859.73
#Sta/Elev= 30
  4340.9  460.35  4695.9  461.09  4839.2  456.87  4861.1  448.96  4888.2  432.23
  4922.5  424.65  4923.7  424.47  5027.1  420.56  5029.8  420.06  5033.1  420.56
  5090.9  424.89  5102.3   425.6  5125.7     428  5151.7  434.19  5161.8  430.63
  5173.3  433.33  5229.6   456.5  5359.5  457.91  5364.5  454.34  5422.3  458.19
  5427.3  454.67    5485  458.99  5490.1  455.35  5605.5  459.53  5831.6     469
  6075.4   477.2  6114.4     475    6134  474.69  6138.2  477.66  6167.2   476.5
#Mann= 11 ,-1 , 0
  4340.9      .1       0  4695.9     .15       0  4923.7      .1       0
  5027.1     .07       0  5033.1      .1       0  5102.3     .16       0
  5125.7      .1       0  5605.5     .08       0  5831.6      .1       0
  6114.4     .05       0    6134     .08       0
Bank Sta=4922.5,5090.9
XS Rating Curve= 0 ,0
Exp/Cntr=0.3,0.1

Type RM Length L Ch R = 1 ,40828   ,562,562,562
BEGIN DESCRIPTION:
MILL BRANCH 73.0
END DESCRIPTION:
XS GIS Cut Line= 4
      3675929.06       10779346.      3675286.75     10779486.61
      3674868.34     10779549.11      3674000.26     10779700.16
#Sta/Elev= 30
  4191.1  466.13  4436.2  467.52  4699.5  454.33  4704.6  457.21  4743.3  453.16
  4748.4  456.51  4792.3  451.06  4797.4  454.85  4841.3  447.24  4848.6  450.62
  4855.8  444.92  4894.6  429.49  4916.5  424.52  4959.3  420.16  4994.4  419.07
  4997.1  418.57  5000.4  419.07  5098.5  420.95  5128.8  425.93  5199.6  438.46
  5245.1  450.66  5300.8  447.77  5366.1  451.26  5398.7  449.25  5461.8  452.35
  5702.2  465.82  5827.8  471.75  5832.9  469.37  5929.3  472.08  6152.8  473.76
#Mann= 9 ,-1 , 0
  4191.1      .1       0  4894.6     .16       0  4959.3      .1       0
  4994.4     .07       0  5000.4      .1       0  5398.7     .05       0
  5461.8      .1       0  5702.2     .05       0  5929.3      .1       0
Bank Sta=4916.5,5128.8
XS Rating Curve= 0 ,0
Exp/Cntr=0.3,0.1

Type RM Length L Ch R = 1 ,40266   ,448,448,448
BEGIN DESCRIPTION:
MILL BRANCH 72.0
END DESCRIPTION:
XS GIS Cut Line= 2
      3675284.05     10778902.02      3674659.09     10779072.14
#Sta/Elev= 30
  4673.8  449.89  4709.5  447.77  4764.3  442.35  4792.4  438.89  4798.8  437.14
  4813.1  436.39  4885.7  424.33  4927.1  418.26  4947.5  416.58  4968.6  416.92
    5007  415.33  5009.8  414.83    5013  415.33  5032.2  416.91  5066.8     416
    5093  419.38  5146.3  422.84  5155.1  424.88  5175.7  426.86  5180.9   426.4
  5186.2  427.87    5207  429.48  5215.5  431.52  5220.7  431.14  5238.1  433.71
  5255.3  439.14  5260.5  438.51  5269.1  441.04    5295  444.32  5321.5  445.48
#Mann= 3 ,-1 , 0
  4673.8     .16       0    5007     .07       0    5013     .16       0
Bank Sta=4885.7,5155.1
XS Rating Curve= 0 ,0
Exp/Cntr=0.3,0.1

Type RM Length L Ch R = 1 ,39818   ,503,503,503
BEGIN DESCRIPTION:
MILL BRANCH 71.0
END DESCRIPTION:
XS GIS Cut Line= 3
      3675149.57     10778410.21      3674899.61     10778560.19
      3674699.62     10778660.18
#Sta/Elev= 30
  4720.6  446.82  4734.2  446.09  4743.9  444.31  4771.1     442  4802.2  436.57
  4813.9  435.22  4837.2  430.76  4860.5  428.27  4881.9  424.13  4895.5  421.26
  4915.6  418.49  4924.2  417.37  4930.5  416.54  4964.4  415.33  4967.2  414.83
  4970.4  415.33  5032.9  415.33  5042.9  417.78  5048.4  416.71  5056.8  417.47
  5070.8   416.6  5087.6  417.84  5109.9  421.12  5137.9  423.92  5160.2  426.67
  5168.6  428.88    5177  429.27  5182.6  431.55    5191  433.42  5235.7  438.72
#Mann= 6 ,-1 , 0
  4720.6     .16       0  4915.6     .12       0  4924.2     .05       0
  4964.4    .033       0  4970.4     .05       0  5032.9     .16       0
Bank Sta=4881.9,5137.9
XS Rating Curve= 0 ,0
Exp/Cntr=0.3,0.1

Type RM Length L Ch R = 1 ,39315   ,379,379,379
BEGIN DESCRIPTION:
MILL BRANCH 70.0
END DESCRIPTION:
XS GIS Cut Line= 3
      3675193.12     10778263.75      3674867.64     10778070.63
      3674383.02     10778098.75
#Sta/Elev= 30
  4571.7   444.5  4686.4  444.74  4738.6  442.33  4781.9  437.51  4796.7  435.25
  4809.1  431.83  4818.9  431.18  4867.6  423.75  4883.2  422.55  4889.7  420.95
  4912.9  418.18  4941.6  416.45  4943.1  415.33  4945.9  414.83  4949.1  415.33
  5016.7  415.33  5078.4  416.47  5118.5  424.86  5128.5  427.59  5148.5  429.94
  5158.5   432.6  5168.6  433.76  5197.5   436.6  5202.6  435.95  5218.6  437.75
    5258   439.3  5293.4  439.72  5328.8  441.63  5368.9  442.01  5435.6  446.57
#Mann= 7 ,-1 , 0
  4571.7     .16       0  4912.9     .05       0  4943.1    .033       0
  4949.1     .05       0  5016.7     .12       0    5258     .16       0
  5293.4     .12       0
Bank Sta=4867.6,5118.5
XS Rating Curve= 0 ,0
Exp/Cntr=0.3,0.1

Type RM Length L Ch R = 1 ,38936   ,507,507,507
BEGIN DESCRIPTION:
MILL BRANCH 69.0
END DESCRIPTION:
XS GIS Cut Line= 3
      3675149.63     10777710.19      3674749.61     10777710.19
      3674449.64     10777960.17
#Sta/Elev= 30
  4604.6  444.08  4694.6  434.15  4714.6  430.89  4740.9  428.35  4764.6  425.06
  4774.6  422.84  4784.6  422.38  4814.6  418.12  4839.9  416.72  4861.6  415.33
  4864.4  414.83  4867.6  415.33    5168  415.33  5173.9  417.22  5196.6   416.3
  5217.5  418.74  5225.3  418.93  5231.8  421.08  5246.1  421.34  5252.6  423.21
  5260.4  423.39  5266.9  424.56  5274.7  425.01  5281.2  426.81    5289  426.92
  5295.6  429.15  5324.2  431.48    5345  435.33  5367.1   437.1  5395.1  440.46
#Mann= 6 ,-1 , 0
  4604.6     .12       0  4740.9     .16       0  4839.9     .05       0
  4861.6    .033       0  4867.6     .05       0  5173.9     .12       0
Bank Sta=4764.6,5266.9
XS Rating Curve= 0 ,0
Exp/Cntr=0.3,0.1

Type RM Length L Ch R = 1 ,38429   ,44,44,44
BEGIN DESCRIPTION:
Mapping XS 113b1a9b
END DESCRIPTION:
XS GIS Cut Line= 2
      3675369.34     10777263.48      3674239.14      10777173.2
#Sta/Elev= 30
  4425.1  457.78    4475  455.09  4535.2  448.18  4545.2  448.46  4555.2   445.6
  4595.4  439.15  4625.5  436.09  4660.1  429.97  4664.8  428.56  4695.7  425.08
  4705.7  421.87  4715.8   421.6  4775.7  415.44  4780.7  416.34    4793  415.33
  4795.8  414.83    4799  415.33  4961.8  415.33  5026.7  415.33  5056.8   416.8
  5066.9  415.33    5107  415.33  5137.1  416.89  5154.7  415.52  5159.7  417.15
  5197.3  417.78  5265.6   416.2  5448.1  423.69  5528.3  425.77  5558.9  429.08
#Mann= 7 ,-1 , 0
  4425.1     .12       0  4660.1     .16       0  4664.8     .05       0
    4793     .07       0    4799     .05       0  4961.8     .16       0
  5265.6     .05       0
Bank Sta=4695.7,5448.1
XS Rating Curve= 0 ,0
Exp/Cntr=0.3,0.1

Type RM Length L Ch R = 1 ,38385   ,62,62,62
BEGIN DESCRIPTION:
Mapping XS cb2fab45
END DESCRIPTION:
XS GIS Cut Line= 2
      3675370.27     10777225.29      3674219.22     10777122.86
#Sta/Elev= 30
  4434.7  455.31  4440.1  454.81  4515.7  451.18  4525.7  448.89  4544.7  446.53
  4549.7  447.46  4555.8  445.75    4586  442.74  4594.9   440.7    4606  439.83
  4636.2  433.63  4673.9  428.65  4686.4   425.9  4706.4  423.25  4736.5  421.97
    4773  422.53    4775  421.88  4777.8  421.38    4781  421.88  4786.7  422.92
  4796.8  422.98  4971.1     423  5067.9   423.4  5188.3  424.29  5286.5  422.64
  5341.2  422.06  5389.1  424.13  5439.3  424.86  5519.6  427.95  5590.3  432.81
#Mann= 8 ,-1 , 0
  4434.7     .16       0  4440.1     .12       0  4594.9     .16       0
  4673.9     .05       0    4775     .07       0    4781     .05       0
  4971.1     .16       0  5286.5     .05       0
Bank Sta=4706.4,5067.9
XS Rating Curve= 0 ,0
Exp/Cntr=0.3,0.1

Type RM Length L Ch R = 1 ,38323   ,355,355,355
BEGIN DESCRIPTION:
MILL BRANCH 68.0
END DESCRIPTION:
XS GIS Cut Line= 2
      3675397.98     10777179.28      3674248.72     10777061.23
#Sta/Elev= 30
  4435.5  450.97  4472.3  451.24  4477.3  449.93  4554.5  446.58  4624.9   438.3
  4670.7  431.31  4685.2  430.61  4700.9  427.76  4750.8  421.32  4876.2  410.82
  4916.4  408.88  4986.8  408.88  5003.9   405.7  5006.6   405.2  5009.9   405.7
  5016.9  406.58    5037  413.24  5087.3  419.69  5107.4  421.32  5140.4  421.54
  5248.1  421.38  5260.8  418.54  5298.4  412.88  5329.1  414.93  5338.6  418.67
    5360  423.46  5479.3  427.16  5548.3  431.07  5553.4  432.73  5590.8  434.58
#Mann= 7 ,-1 , 0
  4435.5     .16       0  4700.9     .05       0  4750.8     .16       0
  5003.9     .07       0  5009.9     .16       0  5140.4     .16       0
  5329.1     .05       0
Bank Sta=4986.8,5037
XS Rating Curve= 0 ,0
Exp/Cntr=0.3,0.1

Type RM Length L Ch R = 1 ,37968   ,463,463,463
BEGIN DESCRIPTION:
MILL BRANCH 67.0
END DESCRIPTION:
XS GIS Cut Line= 2
      3675437.97     10776881.54      3674517.83     10776787.79
#Sta/Elev= 30
  4549.5  450.28  4588.1  449.34  4618.2  446.86  4648.4  445.88  4698.6  440.01
  4738.8  436.89  4748.9  435.02  4799.1  430.43  4879.6  418.48  4889.6  417.94
  4899.7  415.51  4939.9  409.92  4949.9  409.65    4960   407.9  4990.1   406.3
  4997.2  404.91  4999.9  404.41  5003.2  404.91    5006  407.16    5011  407.89
  5084.9  408.24  5120.8   407.5  5171.1  408.45  5227.6  414.64  5299.7  414.35
  5341.9  416.34    5352  417.84    5362  417.96  5452.5  431.25  5474.4   432.5
#Mann= 5 ,-1 , 0
  4549.5     .16       0  4997.2     .07       0  5003.2     .16       0
  5084.9     .12       0  5227.6     .16       0
Bank Sta=4949.9,5011
XS Rating Curve= 0 ,0
Exp/Cntr=0.3,0.1

Type RM Length L Ch R = 1 ,37505   ,391,391,391
BEGIN DESCRIPTION:
MILL BRANCH 66.0
END DESCRIPTION:
XS GIS Cut Line= 4
      3675396.32     10776666.28       3675031.7     10776430.15
      3674889.34     10776426.68      3674528.27     10776530.83
#Sta/Elev= 30
  4463.2  441.25    4495  440.76  4501.5   439.7  4543.7  437.92  4602.2  432.43
  4646.6  425.13  4719.1  417.64  4782.4  408.15  4791.6  406.33  4833.9  405.78
  4876.3  403.75  4969.7  404.37  4986.7  403.05  4989.5  402.55  4992.7  403.05
  5009.7  404.73  5029.7  403.55  5060.5  404.09  5068.2  405.68  5091.8  407.37
  5107.1  409.04  5112.6  411.19    5123  411.67  5140.7  414.46  5154.2  418.08
  5195.8  424.44  5237.5  429.52  5299.9   433.1  5353.3  433.99  5415.8  434.31
#Mann= 4 ,-1 , 0
  4463.2     .16       0  4986.7     .07       0  4992.7     .16       0
  5353.3     .05       0
Bank Sta=4782.4,5091.8
XS Rating Curve= 0 ,0
Exp/Cntr=0.3,0.1

Type RM Length L Ch R = 1 ,37114   ,449,449,449
BEGIN DESCRIPTION:
MILL BRANCH 65.0
END DESCRIPTION:
XS GIS Cut Line= 3
      3675249.58      10775910.2      3674849.61     10776060.19
      3674599.63     10776110.18
#Sta/Elev= 30
  4571.6  430.76    4689  422.13  4732.7  416.84  4752.2  415.98  4757.6  414.14
  4763.8  413.26  4774.5  412.98  4795.8  409.88  4849.2  405.36  4881.3  402.46
    4892  402.78  4898.2  401.27  4913.3  400.56  4928.5  402.01  4958.7  400.82
  4977.4  401.89  4993.1  400.53  4995.8  400.03  4999.1  400.53    5009     402
  5080.4  402.17  5100.7  403.18  5110.9  405.28  5141.5  409.02  5151.7  411.51
  5161.9  412.17  5212.9  422.08  5243.5  426.01  5251.2  428.76  5253.7  428.76
#Mann= 3 ,-1 , 0
  4571.6     .16       0  4993.1     .07       0  4999.1     .16       0
Bank Sta=4849.2,5110.9
XS Rating Curve= 0 ,0
Exp/Cntr=0.3,0.1

Type RM Length L Ch R = 1 ,36665   ,473,473,473
BEGIN DESCRIPTION:
MILL BRANCH 64.0
END DESCRIPTION:
XS GIS Cut Line= 3
      3675149.65     10775660.19      3674749.61     10775660.19
      3674599.57      10775710.2
#Sta/Elev= 30
    4598  425.96    4628   424.2    4638  422.89    4668  420.69    4678  419.28
    4738  413.47    4768  411.67    4788  409.64    4798   409.4    4818  406.82
    4828  404.97    4858  402.21    4888  399.13    4908  398.78    4938  399.24
    4948  397.48    4968  399.46    4978  399.48    4988  396.93  4992.5  396.59
  4995.3  396.09  4998.5  396.59  5029.7  399.22  5050.7  402.46  5071.8  404.67
    5114  410.59  5124.5  414.28  5145.6  418.32  5153.5  420.69  5156.2  420.69
#Mann= 3 ,-1 , 0
    4598     .16       0  4992.5     .07       0  4998.5     .16       0
Bank Sta=4858,5050.7
XS Rating Curve= 0 ,0
Exp/Cntr=0.3,0.1

Type RM Length L Ch R = 1 ,36192   ,528,528,528
BEGIN DESCRIPTION:
MILL BRANCH 63.0
END DESCRIPTION:
XS GIS Cut Line= 3
      3674999.64      10775310.2      3674699.61     10775210.19
      3674449.61     10775360.19
#Sta/Elev= 30
  4682.5  415.56  4703.6  413.04  4724.7   411.8  4735.2  408.99  4777.4  405.02
    4809   400.4  4819.6  399.97  4830.1  398.42  4861.7  396.07  4882.8  396.85
  4956.6  395.95  4977.7  396.96  4988.2  395.84  4993.1  394.37  4995.9  393.87
  4999.1  394.37  5022.1  395.82  5033.7  395.57  5057.1  396.87  5070.7  396.53
  5092.1  398.72  5115.4  399.71  5123.2  401.11  5160.1  403.75  5165.9  404.54
  5181.5  408.76  5187.3  409.11  5208.7  413.11  5255.3  418.58  5290.3  421.48
#Mann= 4 ,-1 , 0
  4682.5     .12       0  4777.4     .16       0  4993.1     .07       0
  4999.1     .16       0
Bank Sta=4830.1,5092.1
XS Rating Curve= 0 ,0
Exp/Cntr=0.3,0.1

Type RM Length L Ch R = 1 ,35664   ,16,16,16
BEGIN DESCRIPTION:
Mapping XS e992b69b
END DESCRIPTION:
XS GIS Cut Line= 2
      3675092.06     10774644.99       3674295.1       10774770.
#Sta/Elev= 30
  4529.1  429.78  4557.6  429.06  4612.6  424.46  4642.9  417.44  4663.8  407.26
  4689.9  404.64  4713.8  404.17  4798.3  394.04  4919.4   391.5    4977  394.65
  4982.1   391.9  4992.3  392.53  5014.4  390.83  5017.2  390.33  5020.4  390.83
  5027.6  395.02  5044.7  398.48  5049.8  395.57  5057.9  395.82  5107.3  400.99
  5112.4  398.14    5149  403.44    5194   403.9  5219.9  408.19  5237.7  417.94
  5242.7  415.58  5250.3  418.75  5294.8  421.42  5305.4  421.58  5335.8  422.96
#Mann= 10 ,-1 , 0
  4529.1     .12       0  4557.6     .16       0  4689.9     .05       0
  4798.3     .16       0  4992.3     .05       0  5014.4     .03       0
  5020.4     .05       0    5194     .08       0  5294.8     .05       0
  5305.4     .08       0
Bank Sta=4977,5027.6
XS Rating Curve= 0 ,0
Exp/Cntr=0.3,0.1

Type RM Length L Ch R = 1 ,35648   ,44,44,44
BEGIN DESCRIPTION:
Mapping XS 58e98fde
END DESCRIPTION:
XS GIS Cut Line= 2
      3675089.45     10774629.36      3674287.33     10774754.37
#Sta/Elev= 30
  4526.1  430.98  4549.1  431.83  4606.9  425.93  4667.6  411.77  4683.6  406.14
  4756.2  402.02  4761.3  399.47    4819  401.59  4824.1  398.16  4859.9  400.37
  4877.4  398.36  4910.5  398.58  4920.6  395.37  4949.8  400.21  4954.8  397.19
  4971.3  397.18  4981.4  394.66    4986  392.99  4998.6   390.5  5001.4     390
  5004.6   390.5  5022.7  394.87    5032  398.57  5052.2  401.57  5085.6  400.52
  5187.6  403.53    5204  403.78  5244.5  418.58  5288.4  420.69  5337.9  421.58
#Mann= 9 ,-1 , 0
  4526.1     .12       0  4549.1     .16       0  4683.6     .05       0
  4877.4     .16       0    4986     .05       0  4998.6     .03       0
  5004.6     .05       0  5187.6     .08       0  5288.4     .05       0
#XS Ineff= 2 , 0
         4945.45  400.06
Permanent Ineff=
       F       F
Bank Sta=4981.4,5022.7
XS Rating Curve= 0 ,0
Exp/Cntr=0.3,0.1

Type RM Length L Ch R = 1 ,35604   ,313,313,313
BEGIN DESCRIPTION:
Mapping XS 9a529631
END DESCRIPTION:
XS GIS Cut Line= 2
      3675081.13     10774585.09       3674273.3     10774714.96
#Sta/Elev= 30
  4519.2  433.13  4522.5  432.86  4525.9  432.63  4584.7  428.49  4641.5  418.23
  4646.6  416.88  4652.4  412.34  4666.6  409.32  4708.5  402.67  4753.7  398.34
  4814.5  395.77    4855  395.27  4865.1   396.7  4885.4  394.63  4915.7  396.02
    4956  393.67  4966.4  396.21  4976.5  393.62    5014  390.06  5016.8  389.56
    5020  390.06  5057.5  395.12  5171.1  402.63  5199.3  403.96  5208.6  408.46
  5213.7  406.53  5219.6     413  5229.7  414.81    5272   417.5  5337.4  419.66
#Mann= 8 ,-1 , 0
  4519.2     .16       0  4522.5     .12       0  4525.9     .16       0
  4666.6     .05       0    5014     .03       0    5020     .05       0
  5171.1     .08       0    5272     .05       0
#XS Ineff= 2 , 0
          4965.2  396.12
Permanent Ineff=
       F       F
Bank Sta=4976.5,5057.5
XS Rating Curve= 0 ,0
Exp/Cntr=0.3,0.1

Type RM Length L Ch R = 1 ,35291   ,89,89,89
BEGIN DESCRIPTION:
MILL BRANCH 62.0
END DESCRIPTION:
XS GIS Cut Line= 3
      3674977.49     10774413.22      3674427.96     10774374.16
      3673973.43     10774846.87
#Sta/Elev= 30
    4500  424.67  4534.3  420.93    4558  419.44  4588.1  410.03  4613.2   406.6
  4758.9  401.81  4828.7   393.6    4939  390.73  4969.1  392.57  4996.1  388.33
  4998.9  387.83  5002.1  388.33  5019.2  392.48  5089.3  394.14  5167.1  399.28
  5186.1   400.2  5216.6     401  5252.2  406.56  5266.3  406.87  5273.2  403.01
  5287.4  402.31  5301.5  402.38  5317.2  406.13    5344  409.12  5421.7  410.97
  5471.3  416.85    5549  418.15  5579.3  423.93  5662.2  430.41  5706.7  429.74
#Mann= 8 ,-1 , 0
    4500     .16       0  4534.3     .05       0  4996.1     .03       0
  5002.1     .05       0  5167.1     .08       0  5186.1     .05       0
  5317.2     .16       0  5579.3     .08       0
Bank Sta=4828.7,5089.3
XS Rating Curve= 0 ,0
Exp/Cntr=0.3,0.1

Type RM Length L Ch R = 1 ,35202   ,380,380,380
BEGIN DESCRIPTION:
MILL BRANCH 61.0
END DESCRIPTION:
XS GIS Cut Line= 3
      3674943.07     10774317.63      3674419.61     10774286.38
      3673896.17     10774088.46
#Sta/Elev= 30
  4526.6  427.11  4550.1  425.78  4566.3  419.98  4640.3  419.03  4670.3  416.81
  4680.3  415.21  4688.3  411.02  4710.4  402.28  4850.6  393.75  4880.7  391.78
  4970.8   391.5  4990.9  390.03  4997.9  387.08  5000.7  386.58  5003.9  387.08
  5010.9  389.72  5020.9  390.42  5200.9  392.52  5211.4  395.27  5220.3   401.6
  5228.1  402.43  5232.7  403.28  5250.5  398.04  5255.9  401.78  5275.3  408.96
  5280.7  408.91  5286.2  414.78  5318.3  419.42  5479.3  429.99  5610.6  439.13
#Mann= 6 ,-1 , 0
  4526.6     .08       0  4688.3     .05       0  4997.9     .03       0
  5003.9     .05       0  5228.1     .16       0  5479.3     .05       0
Bank Sta=4850.6,5200.9
XS Rating Curve= 0 ,0
Exp/Cntr=0.3,0.1

Type RM Length L Ch R = 1 ,34822   ,109,109,109
BEGIN DESCRIPTION:
Mapping XS 814703ea
END DESCRIPTION:
XS GIS Cut Line= 2
      3674943.08     10774262.96      3674054.99      10773632.7
#Sta/Elev= 30
  4415.8  427.24  4463.4  420.61  4549.5  414.83  4555.6     412  4564.3  412.24
  4570.4  407.79  4620.8  406.43  4650.4  399.53  4763.1  394.86  4800.2  395.56
    4814  393.27  4879.2  389.45  4980.1  389.05  4991.8  386.78  4994.6  386.28
  4997.8  386.78  5066.2  392.32  5094.5  393.86  5117.6  395.99  5173.2  400.62
  5180.3  404.68  5238.4  413.98  5319.5  421.07  5339.3  421.58  5345.4   419.5
  5360.2  422.27  5424.5  423.35  5431.5  420.73    5472  422.81  5504.8  418.07
#Mann= 9 ,-1 , 0
  4415.8     .08       0  4763.1     .05       0  4991.8     .04       0
  4997.8     .05       0  5066.2     .08       0  5117.6     .05       0
  5319.5     .16       0  5424.5     .08       0    5472     .05       0
#XS Ineff= 2 , 0
         4767.54  395.92
Permanent Ineff=
       F       F
Bank Sta=4814,5094.5
XS Rating Curve= 0 ,0
Exp/Cntr=0.3,0.1

Type RM Length L Ch R = 1 ,34713   ,392,392,392
BEGIN DESCRIPTION:
MILL BRANCH 60.0
END DESCRIPTION:
XS GIS Cut Line= 2
      3675031.59       10774177.      3674096.71     10773549.41
#Sta/Elev= 30
  4416.5  430.09  4596.7  419.45  4653.4  416.02  4700.2  407.62  4776.4  397.63
  4840.4  392.88  4858.2  391.72  4923.8  390.31  4974.4  389.91    4985   389.7
  4995.5  385.45  4998.2  384.95  5001.5  385.45  5043.4  389.93  5049.5  392.91
  5079.4  392.28  5110.5  392.73  5178.5  394.94  5206.8  398.78  5244.5  401.99
  5250.5  404.42  5297.1  407.03    5323  408.38  5367.5  411.27  5373.5  414.32
  5388.5  412.32  5394.5  414.74  5403.5  414.71  5483.8  411.68  5542.5  411.67
#Mann= 13 ,-1 , 0
  4416.5     .12       0  4596.7     .08       0  4700.2     .12       0
  4858.2     .08       0  4923.8     .12       0  4974.4     .08       0
  4995.5     .07       0  5001.5     .08       0  5110.5     .16       0
  5206.8     .05       0  5297.1     .16       0    5323     .08       0
  5483.8     .16       0
Bank Sta=4840.4,5079.4
XS Rating Curve= 0 ,0
Exp/Cntr=0.3,0.1

Type RM Length L Ch R = 1 ,34321   ,594,594,594
BEGIN DESCRIPTION:
MILL BRANCH 59.0
END DESCRIPTION:
XS GIS Cut Line= 3
      3675149.58     10773560.19      3674749.61     10773610.19
      3674349.59     10773210.17
#Sta/Elev= 30
  4574.6  426.34    4693  413.87  4698.5  412.48  4735.8  408.16    4766  403.02
  4778.6  402.73  4806.4  399.17  4854.2  395.69  4859.3  396.43  4896.6  394.93
  4957.5  391.77  4967.6  389.58  4981.2  388.37  4988.8  384.82  4991.6  384.32
  4994.8  384.82  5020.1  389.22  5034.3  391.87  5048.4  391.03  5076.7  385.99
  5110.2  386.05  5232.2  386.31  5288.8   387.6    5303  391.24  5331.2  393.41
  5345.7   396.9  5387.8  400.79  5417.1  406.05  5500.9  417.89  5543.4  420.99
#Mann= 8 ,-1 , 0
  4574.6     .12       0  4698.5     .16       0  4896.6     .12       0
  4988.8     .07       0  4994.8     .12       0  5110.2     .07       0
  5345.7     .12       0  5417.1     .16       0
Bank Sta=4967.6,5020.1
XS Rating Curve= 0 ,0
Exp/Cntr=0.3,0.1

Type RM Length L Ch R = 1 ,33727   ,290,290,290
BEGIN DESCRIPTION:
MILL BRANCH 58.0
END DESCRIPTION:
XS GIS Cut Line= 3
      3675310.72     10773473.94       3674839.4     10773143.23
      3674373.89     10773049.61
#Sta/Elev= 30
  4516.4  427.51  4542.2  425.78  4548.7   426.8  4554.8  425.11  4578.3   424.2
  4584.4  422.07    4614  420.82  4620.1  418.93    4635  419.67  4685.5  411.31
  4764.1  401.54  4807.5  396.46  4813.6  394.49  4885.1  389.19  4929.5  385.41
    4998  384.57  5000.8  384.07    5004  384.57  5021.9  386.02  5175.7  386.33
    5232  387.51  5255.2  386.55    5288  388.75  5333.8  392.44  5418.4  403.08
  5471.3  407.78  5520.4  413.01  5537.2  416.13  5542.3  414.72    5567  417.65
#Mann= 6 ,-1 , 0
  4516.4     .16       0  4764.1     .12       0    4998     .07       0
    5004     .12       0  5175.7     .16       0  5471.3      .1       0
Bank Sta=4885.1,5288
XS Rating Curve= 0 ,0
Exp/Cntr=0.3,0.1

Type RM Length L Ch R = 1 ,33437   ,447,447,447
BEGIN DESCRIPTION:
MILL BRANCH 57.0
END DESCRIPTION:
XS GIS Cut Line= 2
      3675511.24     10773359.35      3674474.86     10772520.87
#Sta/Elev= 30
  4477.4  433.52  4480.7  433.52    4485  431.52  4499.4  431.58  4593.7  419.84
  4606.5  419.44  4684.8  408.92  4698.2  406.06  4773.8  397.47    4947  387.32
    5011  383.84  5032.6  385.19  5115.1  383.12  5117.8  382.62  5121.1  383.12
    5246  386.14  5295.6  385.98    5310  387.83  5373.9  388.92  5401.2  393.17
  5423.5  395.37  5444.3  399.05  5473.1  400.47  5501.8  400.98  5594.5   396.9
  5650.6  397.85  5757.7  404.88  5778.7  407.05  5786.4     409  5810.5  410.65
#Mann= 6 ,-1 , 0
  4477.4     .12       0  4593.7     .16       0  4773.8     .12       0
  5115.1     .07       0  5121.1     .12       0  5401.2     .16       0
Bank Sta=4947,5310
XS Rating Curve= 0 ,0
Exp/Cntr=0.3,0.1

Type RM Length L Ch R = 1 ,32990   ,567,567,567
BEGIN DESCRIPTION:
MILL BRANCH 56.0
END DESCRIPTION:
XS GIS Cut Line= 3
      3675932.77     10772819.89      3675240.01     10772736.55
      3674479.62     10771970.95
#Sta/Elev= 30
  4211.9  438.19  4466.9  419.18  4584.4  405.82  4678.4  401.28  4708.6  395.77
  4718.7   390.8  4753.8  390.21  4809.3  384.17    4841  381.95  4935.6  383.06
  4989.2  381.34    4992  380.84  4995.2  381.34  5034.6  381.81  5048.8  384.08
  5119.5  381.82  5154.9  384.34  5239.7  381.66  5282.1   383.7  5381.1  382.06
  5451.9  389.23  5543.8   402.2  5586.2  404.84  5628.6  404.33  5635.7  402.14
  5642.8  403.69  5649.8  401.02  5656.9  404.23  5706.4  403.04  5988.7  422.53
#Mann= 3 ,-1 , 0
  4211.9     .12       0  4989.2     .07       0  4995.2     .12       0
Bank Sta=4809.3,5048.8
XS Rating Curve= 0 ,0
Exp/Cntr=0.3,0.1

Type RM Length L Ch R = 1 ,32423   ,539,539,539
BEGIN DESCRIPTION:
MILL BRANCH 55.0
END DESCRIPTION:
XS GIS Cut Line= 2
      3675812.94     10772621.98      3674913.23      10771956.3
#Sta/Elev= 30
  4507.6  421.71    4554  418.31  4668.8  404.86  4810.7  393.49  4869.2  391.14
  4897.4  386.13  4910.9  386.75    4961  381.37  5003.9  379.64  5032.2   380.1
  5075.8  380.43  5108.3  377.76    5111  377.26  5114.3  377.76  5211.5  380.19
  5233.2  378.25  5246.9  380.27  5255.3  378.56  5305.4  381.36  5340.9  378.87
  5382.6  381.79  5426.5  385.13  5441.1  391.03  5455.7  392.29    5462  395.52
  5476.6  395.51  5482.8  398.37  5512.1  401.58  5597.6  405.54  5626.8  403.87
#Mann= 5 ,-1 , 0
  4507.6     .12       0  5003.9     .16       0  5032.2     .12       0
  5108.3     .07       0  5114.3     .12       0
Bank Sta=4961,5382.6
XS Rating Curve= 0 ,0
Exp/Cntr=0.3,0.1

Type RM Length L Ch R = 1 ,31884   ,434,434,434
BEGIN DESCRIPTION:
MILL BRANCH 54.0
END DESCRIPTION:
XS GIS Cut Line= 3
       3675849.6     10772160.18      3675499.61     10771960.19
       3675099.6     10771560.18
#Sta/Elev= 30
  4605.1  418.98  4618.8  418.22  4656.2  413.12  4662.7  410.99  4693.6  407.17
    4721  402.11  4736.8  401.33  4743.3  399.33  4766.3  396.04    4780  395.22
  4795.8   391.6    4839     387  4860.6  382.55    4870  382.39  4882.2     380
  4898.1  379.16  4904.5  377.83  4957.1  375.35  4994.5  375.35  5002.3   373.9
  5005.1   373.4  5008.3   373.9  5050.6  375.36  5135.5  375.71  5262.8  378.62
  5319.3   381.4    5489   395.5  5500.7  397.41  5531.5  399.83  5573.9  405.85
#Mann= 4 ,-1 , 0
  4605.1     .12       0  5002.3     .07       0  5008.3     .12       0
  5500.7     .16       0
Bank Sta=4898.1,5262.8
XS Rating Curve= 0 ,0
Exp/Cntr=0.3,0.1

Type RM Length L Ch R = 1 ,31450   ,317,317,317
BEGIN DESCRIPTION:
MILL BRANCH 53.0
END DESCRIPTION:
XS GIS Cut Line= 3
      3675899.63     10771960.22      3675649.61     10771560.19
      3675449.64     10771410.21
#Sta/Elev= 30
  4551.8  402.76  4610.8  397.88  4653.8  390.05  4675.1  387.45  4690.4  384.07
  4740.5  377.37  4754.1   375.8  4848.4  374.22  4863.7  374.94  4921.5   373.3
  4942.8  374.09  4970.4  372.85  4973.2  372.35  4976.4  372.85  5030.8  373.41
  5080.8  377.11    5110  380.45  5116.2  382.18  5130.8  382.99  5145.4  386.07
  5151.7  386.15  5180.8   392.7  5187.1  392.99  5195.4  396.07  5216.2  398.81
  5223.5  401.71  5237.1  403.83  5245.4  407.05    5260  410.55  5273.5  411.58
#Mann= 4 ,-1 , 0
  4551.8     .12       0  4970.4     .07       0  4976.4     .12       0
  5180.8     .16       0
Bank Sta=4740.5,5080.8
XS Rating Curve= 0 ,0
Exp/Cntr=0.3,0.1

Type RM Length L Ch R = 1 ,31133   ,874,874,874
BEGIN DESCRIPTION:
MILL BRANCH 52.0
END DESCRIPTION:
XS GIS Cut Line= 2
       3676309.6     10771628.75      3675387.67     10771107.88
#Sta/Elev= 30
  4430.9  416.61  4476.6  414.65  4534.2  408.74  4577.5  400.05  4614.7  396.07
  4626.5  393.11  4664.1  387.95  4695.1  385.39  4775.5  374.99  4809.9  373.41
  4922.5  373.52  4981.7   371.9  4987.5  371.52  4990.7  369.81  4993.4  369.31
  4996.7  369.81    5025  372.57  5052.4  371.93  5127.6  374.35  5192.5  379.79
  5223.4  383.74  5235.8  383.15  5280.8  390.22  5312.9  392.58  5384.2  399.36
  5407.2  402.32  5413.4  404.51  5419.2  404.28  5472.6   411.9  5489.8  413.05
#Mann= 5 ,-1 , 0
  4430.9     .16       0  4476.6     .12       0  4990.7     .07       0
  4996.7     .12       0  5312.9     .16       0
Bank Sta=4775.5,5127.6
XS Rating Curve= 0 ,0
Exp/Cntr=0.3,0.1

Type RM Length L Ch R = 1 ,30259   ,265,265,265
BEGIN DESCRIPTION:
MILL BRANCH 51.0
END DESCRIPTION:
XS GIS Cut Line= 4
      3676372.09     10771545.42      3676028.33     10770623.53
      3675866.88     10770519.36      3674924.34     10770904.71
#Sta/Elev= 30
    3900  415.65  4032.1  408.53  4178.4  395.13  4208.7  389.74    4355  377.55
  4551.2   371.6  4716.7  372.92  4998.4  366.97  5001.1  366.47  5004.4  366.97
  5328.1  372.12  5369.4  372.68  5472.8  376.89  5536.4  388.31  5559.2  390.13
  5580.8  395.86  5637.1  397.99  5702.1  399.31  5769.1  395.92  5815.6  395.66
    5857  395.09    5905  399.88  5910.5  395.41  5926.6  394.59  5934.5     400
  5958.5  407.36  6019.9  414.27  6031.5  414.95  6070.8  416.13  6094.3  413.95
#Mann= 9 ,-1 , 0
    3900     .16       0  4998.4     .07       0  5004.4     .16       0
  5369.4     .16       0  5637.1     .05       0  5769.1     .12       0
  5815.6     .05       0  6019.9     .16       0  6031.5     .12       0
#XS Ineff= 2 , 0
         4706.82  381.18
Permanent Ineff=
       F       F
Bank Sta=4716.7,5328.1
XS Rating Curve= 0 ,0
Exp/Cntr=0.3,0.1

Type RM Length L Ch R = 1 ,29994   ,413,413,413
BEGIN DESCRIPTION:
MILL BRANCH 50.0
END DESCRIPTION:
XS GIS Cut Line= 3
      3676599.64     10770660.21      3675999.61     10770310.19
      3675399.62     10770110.19
#Sta/Elev= 30
  4297.7  387.82  4370.1  384.26  4391.6   381.3  4401.5  381.13  4459.8  374.95
    4466  373.06  4481.7  372.09    4509  371.97  4517.7  372.76  4552.4  371.51
  4795.6  369.11  4830.3  369.97    4963  366.46  4978.7  367.15  4989.5  366.01
    5024  366.79  5087.2  366.47  5094.8  365.66  5097.5  365.16  5100.8  365.66
  5129.4   368.7  5245.3  370.79    5411  372.08  5466.7  374.03  5508.9  373.49
  5519.4  374.18  5582.7  382.96  5593.2   383.6  5614.3  388.26  5624.8   388.6
#Mann= 4 ,-1 , 0
  4297.7     .16       0  5094.8     .07       0  5100.8     .16       0
    5411     .16       0
#XS Ineff= 2 , 0
         4826.36  377.77
Permanent Ineff=
       F       F
Bank Sta=4830.3,5245.3
XS Rating Curve= 0 ,0
Exp/Cntr=0.3,0.1

Type RM Length L Ch R = 1 ,29581   ,490,490,490
BEGIN DESCRIPTION:
MILL BRANCH 49.0
END DESCRIPTION:
XS GIS Cut Line= 3
       3676749.6     10770510.18      3676149.61     10769960.19
      3674949.64     10769960.19
#Sta/Elev= 30
  4175.2  396.72  4324.1  389.92  4444.3  379.03  4479.5  378.43  4571.4  371.81
  4578.8  370.32  4621.3  371.33  4762.5  367.77  4868.6  368.06  5016.1  365.14
  5018.9  364.64  5022.1  365.14  5179.1  367.56  5249.1  365.54  5269.1  367.92
  5389.1   367.3  5527.9  369.84  5579.1  371.27  5589.1  369.53  5599.1  371.67
  5659.1  378.01  5669.1  380.57  5709.1  384.41  5779.1  394.67  5839.1   401.5
  5869.1  402.94  5902.2   408.8  5909.2  409.45  5989.1  421.97  6189.1  439.17
#Mann= 6 ,-1 , 0
  4175.2     .16       0  5016.1     .07       0  5022.1     .16       0
  5527.9     .16       0  5902.2     .12       0  5909.2     .16       0
#XS Ineff= 2 , 0
         4754.26  383.63
Permanent Ineff=
       F       F
Bank Sta=4571.4,5599.1
XS Rating Curve= 0 ,0
Exp/Cntr=0.3,0.1

Type RM Length L Ch R = 1 ,29091   ,296,296,296
BEGIN DESCRIPTION:
MILL BRANCH 48.0
END DESCRIPTION:
XS GIS Cut Line= 3
      3677379.07     10769435.59      3675799.17     10769609.21
      3674835.66     10769834.89
#Sta/Elev= 30
  3607.1  417.07  3672.6  413.53  3746.8  410.36  3948.6  402.46  4079.4  392.69
  4200.1  391.01  4310.8  382.02  4391.3  371.89  4431.9  370.74    4606  363.77
  4608.7  363.27    4612  363.77    4700  366.81  4705.1  364.35  4723.2  366.15
  4763.5  363.88  4887.2  365.93  4904.3  363.85  4944.6  363.79  5377.6  366.13
  5487.3  366.37  5529.8   370.8  5740.4  393.52  5832.2  400.51    5915  410.91
  5956.1  418.11    6028  439.61  6054.8  441.31  6059.9  443.47  6186.1  445.54
#Mann= 6 ,-1 , 0
  3607.1     .16       0  3672.6     .05       0  3746.8     .16       0
    4606     .07       0    4612     .16       0  5377.6     .16       0
Bank Sta=4431.9,5529.8
XS Rating Curve= 0 ,0
Exp/Cntr=0.3,0.1

Type RM Length L Ch R = 1 ,28795   ,540,540,540
BEGIN DESCRIPTION:
MILL BRANCH 47.0
END DESCRIPTION:
XS GIS Cut Line= 3
      3677379.05     10769218.58      3675851.25     10769322.75
      3674636.01     10769131.78
#Sta/Elev= 30
  3576.6  421.05  3633.3  417.79  3756.7  412.44  3906.8  401.77  4107.3  396.29
  4317.8  378.55  4478.1  370.93  4618.5  364.62  4678.6  363.62  5019.4  363.35
  5069.5  364.68  5116.7  363.29  5119.5  362.79  5122.7  363.29  5514.5  365.15
    5555  364.06  5747.3  370.37  5801.9  372.59  5864.5  378.02  6020.7  381.88
  6062.3  384.81  6124.9  390.86  6162.4  396.64  6192.7  403.07  6221.4  412.42
  6255.1  421.22  6263.6  424.96  6283.8  428.69  6304.1  430.21  6338.1  429.64
#Mann= 6 ,-1 , 0
  3576.6     .16       0  3633.3     .05       0  3756.7     .12       0
  5116.7     .07       0  5122.7     .12       0  6221.4     .16       0
Bank Sta=4478.1,5747.3
XS Rating Curve= 0 ,0
Exp/Cntr=0.3,0.1

Type RM Length L Ch R = 1 ,28255   ,582,582,582
BEGIN DESCRIPTION:
MILL BRANCH 46.0
END DESCRIPTION:
XS GIS Cut Line= 3
      3676649.56     10768810.19      3676049.61     10768860.19
      3675449.59     10768310.17
#Sta/Elev= 30
  4370.5  391.79  4460.8  376.52    4521  370.54  4581.2  365.11  4621.3  363.48
  4631.4  365.14  4761.8  363.59  4789.4  364.56  4794.4  366.66    4812  364.45
  4842.1  363.87  4952.5   365.4  5000.6  363.11  5128.2  364.45  5196.1  362.87
  5198.9  362.37  5202.1  362.87  5241.7  364.48  5248.5  363.14    5312  363.06
  5368.7  365.11  5510.5  363.96  5553.1  365.18  5602.4   371.1  5630.8  372.18
  5637.6  374.23    5645  373.13  5708.5  381.14  5744.2  383.35  5786.5  392.38
#Mann= 3 ,-1 , 0
  4370.5     .12       0  5196.1     .07       0  5202.1     .12       0
Bank Sta=4521,5602.4
XS Rating Curve= 0 ,0
Exp/Cntr=0.3,0.1

Type RM Length L Ch R = 1 ,27673   ,454,454,454
BEGIN DESCRIPTION:
MILL BRANCH 45.0
END DESCRIPTION:
XS GIS Cut Line= 2
      3676849.55     10768515.46      3675643.76      10768229.2
#Sta/Elev= 30
  4179.4  397.58  4266.9   389.9  4309.1  387.13  4314.3  388.41  4398.7  381.38
  4405.5  379.52    4426  377.45  4435.7  377.95  4539.1  370.22  4678.1  363.76
  4778.9  364.42  4792.2  363.96  4847.4  363.69  4873.2  365.06  4920.5  363.21
  4929.6  364.34  4962.7  362.99  4991.3  364.39  5060.2  362.93    5063  362.43
  5066.2  362.93  5083.8  364.52  5089.3  366.16    5166  364.41  5207.1  370.47
  5221.1  373.08  5264.5  387.24  5268.8  389.34  5310.6   393.9  5418.7  399.65
#Mann= 7 ,-1 , 0
  4179.4     .12       0  4678.1     .16       0  4778.9     .07       0
  4792.2     .12       0  5060.2     .07       0  5066.2     .12       0
  5264.5     .16       0
Bank Sta=4539.1,5207.1
XS Rating Curve= 0 ,0
Exp/Cntr=0.3,0.1

Type RM Length L Ch R = 1 ,27219   ,553,553,553
BEGIN DESCRIPTION:
MILL BRANCH 44.0
END DESCRIPTION:
XS GIS Cut Line= 3
       3676749.6     10768210.19      3676149.61     10767960.19
      3675949.63     10767760.21
#Sta/Elev= 30
  4350.8  391.18  4448.3     384  4556.6  373.12  4589.1  372.01  4601.6  370.24
  4625.4  368.76  4649.3  365.58  4673.1  364.28  4678.5  365.05  4686.6  363.11
  4709.9  363.44  4746.4  364.38  4779.3  365.66  4816.6  364.32  4838.3  366.22
  4900.3  362.66    4903  362.16  4906.3  362.66  4962.3  364.27  4979.1  363.17
  5014.9  363.89  5085.6  362.98  5099.8  363.74  5142.2  369.57  5156.4  373.36
  5198.8  381.95  5212.9  383.08  5241.2  388.23  5280.1  397.75  5283.6  397.75
#Mann= 5 ,-1 , 0
  4350.8     .12       0  4709.9     .16       0  4746.4     .12       0
  4900.3     .07       0  4906.3     .12       0
Bank Sta=4601.6,5156.4
XS Rating Curve= 0 ,0
Exp/Cntr=0.3,0.1

Type RM Length L Ch R = 1 ,26666   ,450,450,450
BEGIN DESCRIPTION:
MILL BRANCH 43.0
END DESCRIPTION:
XS GIS Cut Line= 3
      3676949.65      10767760.2      3676349.61     10767660.19
      3676099.58     10767610.18
#Sta/Elev= 30
  4384.9  411.29  4405.2     410  4463.5  402.51  4486.3  398.69  4516.7  395.38
  4534.5  391.95  4539.5  392.32  4574.9  385.31  4624.5  376.81  4638.4  374.55
  4661.2  373.63  4689.1  370.65  4729.6  366.04  4770.2  364.59  4838.6  363.87
  4843.7  364.77  4861.4  362.98  4932.4  365.09  4942.5  363.41  5000.4  362.83
  5003.2  362.33  5006.4  362.83  5018.7  363.79  5074.8  363.96  5125.8  370.78
  5156.4  377.45  5166.6  380.81  5200.7  386.06  5200.8  386.08  5248.2  391.02
#Mann= 8 ,-1 , 0
  4384.9     .16       0  4463.5     .12       0  4574.9     .16       0
  4624.5     .12       0  5000.4     .07       0  5006.4     .12       0
  5200.7     .16       0  5200.8     .12       0
Bank Sta=4689.1,5125.8
XS Rating Curve= 0 ,0
Exp/Cntr=0.3,0.1

Type RM Length L Ch R = 1 ,26216   ,502,502,502
BEGIN DESCRIPTION:
MILL BRANCH 42.0
END DESCRIPTION:
XS GIS Cut Line= 3
      3676949.61     10767510.19      3676549.61     10767310.19
      3676149.63     10767210.19
#Sta/Elev= 30
  4540.5  400.57  4571.2  398.97  4601.6   395.3  4652.3  388.28  4674.7  382.79
  4683.1  382.11    4697  377.22    4711  375.95  4716.3  374.32  4733.4  370.44
  4743.5  369.91  4772.5  365.29  4794.9  363.28  4864.5  362.61  4867.3  362.11
  4870.5  362.61  4906.7  363.93    4929  363.38  4934.6  364.43    4943  363.24
  4959.3  363.37  5059.9  362.97  5080.5  364.89  5101.1   363.2  5157.8  367.69
  5175.8  369.62  5204.2  370.35  5234.8   373.3  5339.6  382.87    5400  388.51
#Mann= 10 ,-1 , 0
  4540.5     .16       0  4601.6     .12       0  4716.3     .16       0
  4743.5     .12       0  4864.5     .07       0  4870.5     .12       0
  4959.3     .16       0  5157.8     .05       0  5234.8     .12       0
  5339.6     .16       0
Bank Sta=4743.5,5175.8
XS Rating Curve= 0 ,0
Exp/Cntr=0.3,0.1

Type RM Length L Ch R = 1 ,25714   ,450,450,450
BEGIN DESCRIPTION:
MILL BRANCH 41.0
END DESCRIPTION:
XS GIS Cut Line= 3
      3676899.62     10766460.18      3676549.61     10766810.19
      3676049.59      10767110.2
#Sta/Elev= 30
  4500.7  406.36    4529  404.47  4571.4  396.72  4599.7  386.69  4613.8  384.43
    4628  378.45  4642.1  375.85  4656.3  370.93  4670.4  368.68  4712.8  363.12
  4737.2  364.01  4745.3  363.73  4780.6  362.06  4783.3  361.56  4786.6  362.06
  5077.3  362.06  5108.5   363.4  5178.4  362.97  5221.1   366.4  5228.9  365.42
  5261.5  365.48  5287.2  366.01  5361.2  363.36  5379.7  365.48  5403.9  367.88
  5411.6  369.98  5427.2  371.98  5512.7  387.79  5540.2  391.24  5578.8  393.62
#Mann= 10 ,-1 , 0
  4500.7     .12       0  4737.2     .16       0  4745.3     .05       0
  4780.6    .035       0  4786.6     .05       0  5108.5     .16       0
  5261.5     .12       0  5361.2     .16       0  5379.7     .05       0
  5540.2     .12       0
Bank Sta=4670.4,5411.6
XS Rating Curve= 0 ,0
Exp/Cntr=0.3,0.1

Type RM Length L Ch R = 1 ,25264   ,422,422,422
BEGIN DESCRIPTION:
MILL BRANCH 40.0
END DESCRIPTION:
XS GIS Cut Line= 3
      3676899.62     10766410.19      3676349.61     10766410.19
      3675849.62     10766410.19
#Sta/Elev= 30
  4455.9  404.75  4485.9  399.92  4505.9  394.32  4515.9  389.37  4535.9  384.21
  4575.9  377.56  4595.9  374.93  4605.9  374.62  4635.9  369.56  4645.9  369.21
    4670  366.45  4725.9  363.38  4765.9  364.43  4782.9  362.06  4785.7  361.56
  4788.9  362.06    4815  362.06  5222.9  362.06  5235.9  362.06  5245.9  363.81
  5315.9  363.97  5365.9  370.01  5375.9  370.78  5395.9  375.89  5415.9  378.93
  5425.9  381.28  5435.9  386.09    5442  387.15  5455.9  391.13  5505.9  394.67
#Mann= 7 ,-1 , 0
  4455.9     .12       0    4670     .16       0  4782.9    .033       0
  4788.9     .16       0    4815     .05       0  5222.9     .16       0
    5442     .05       0
Bank Sta=4645.9,5365.9
XS Rating Curve= 0 ,0
Exp/Cntr=0.3,0.1
