--- BATSMITH CREEK.prj (project) ---

Proj Title=BATSMITH CREEK Base Level Engineering
Current Plan=p01
Default Exp/Contr=0.3,0.1
English Units
Geom File=g01
Flow File=f01
Plan File=p01
Y Axis Title=Elevation
X Axis Title(PF)=Main Channel Distance
X Axis Title(XS)=Station
BEGIN DESCRIPTION:
BATSMITH CREEK
END DESCRIPTION:
DSS Export Rating Curves= 0
DSS Export Rating Curve Sorted= 0
DSS Export Volume Flow Curves= 0
DXF OffsetX= 0
DXF OffsetY= 0
DXF ScaleX= 1
DXF ScaleY= 10

--- BATSMITH CREEK.p01 (plan) ---

Plan Title=Multiple Run
Short Identifier=Multiple
Geom File=g01
Flow File=f01
Subcritical Flow
K Sum by GR= 0
Std Step Tol= 0.01
Critical Tol= 0.01
Num of Std Step Trials= 20
Max Error Tol= 0.3
Flow Tol Ratio= 0.001
Split Flow NTrial= 30
Split Flow Tol= 0.02
Split Flow Ratio= 0.02
Log Output Level= 0
Friction Slope Method= 1
Unsteady Friction Slope Method= 2
Unsteady Bridges Friction Slope Method= 1
Parabolic Critical Depth
Global Vel Dist=  1 , 1 , 1
Global Log Level= 0
CheckData=True
Encroach Param= -1, 0, 0, 0
BEGIN DESCRIPTION:
Multiple Run
END DESCRIPTION:

--- BATSMITH CREEK.f01 (steady flow) ---

Flow Title=Multiple
Program Version=4.10
Number of Profiles= 7
Profile Names=10-year,25-year,50-year,1pct_min,100-year,1pct_plu,500-year
River Rch & RM=BATSMITH CREEK,Reach-1         ,20125
    2072    2993    3792    3505    4740    6411    7384
River Rch & RM=BATSMITH CREEK,Reach-1         ,17090
    2467    3569    4526    4181    5655    7647    8801
River Rch & RM=BATSMITH CREEK,Reach-1         ,8597
    3037    4423    5635    5225    7066    9556   11090
Boundary for River Rch & Prof#=BATSMITH CREEK,Reach-1         , 1
Up Type= 0
Dn Type= 3
Dn Slope=0.004
Boundary for River Rch & Prof#=BATSMITH CREEK,Reach-1         , 2
Up Type= 0
Dn Type= 3
Dn Slope=0.004
Boundary for River Rch & Prof#=BATSMITH CREEK,Reach-1         , 3
Up Type= 0
Dn Type= 3
Dn Slope=0.004
Boundary for River Rch & Prof#=BATSMITH CREEK,Reach-1         , 4
Up Type= 0
Dn Type= 3
Dn Slope=0.004
Boundary for River Rch & Prof#=BATSMITH CREEK,Reach-1         , 5
Up Type= 0
Dn Type= 3
Dn Slope=0.004
Boundary for River Rch & Prof#=BATSMITH CREEK,Reach-1         , 6
Up Type= 0
Dn Type= 3
Dn Slope=0.004
Boundary for River Rch & Prof#=BATSMITH CREEK,Reach-1         , 7
Up Type= 0
Dn Type= 3
Dn Slope=0.004
DSS Import GetInterval= 0
DSS Import GetPeak= 0
DSS Import FillOption= 0

--- BATSMITH CREEK.g01 (geometry) ---

Geom Title=Existing Conditions
Program Version=4.10

River Reach=BATSMITH CREEK  ,Reach-1
Reach XY= 30
      3632999.61       10617150.      3633303.75       10617159.
       3633600.5       10616891.       3634242.5       10616996.
       3634456.5       10616693.      3634934.75       10616821.
      3635046.25       10616503.      3635614.75       10616561.
      3636487.25       10615701.      3636882.25       10615666.
      3636970.75       10615806.      3637072.25       10615609.
      3637507.25       10615533.      3637680.25       10615255.
       3637883.5       10615347.       3638271.5       10614894.
        3639485.       10614502.      3639718.75       10614665.
       3639974.5       10614512.      3640534.75       10613357.
      3640940.75       10613083.        3642015.       10613281.
      3642533.25       10612957.        3642649.       10613181.
        3643759.       10612440.       3644959.5       10612520.
       3645116.5       10612796.      3646524.25       10613250.
      3646985.25       10612755.      3647538.75       10613036.

Type RM Length L Ch R = 1 ,20125   ,437,437,437
BEGIN DESCRIPTION:
BATSMITH CREEK 42.0
END DESCRIPTION:
XS GIS Cut Line= 3
      3633099.61      10617360.2      3633099.61     10617060.19
      3633049.61      10616960.2
#Sta/Elev= 30
  4732.6  418.68  4762.6  416.62  4782.6  415.64  4812.6  414.91  4832.6  413.65
  4902.6  411.82  4922.6     412  4942.6  411.63  4952.6  410.08  4962.6  409.17
  4972.6  407.33  4982.6  406.26  4992.6  403.47  4999.6  403.24  5002.4  402.74
  5005.6  403.24  5012.6  405.22  5022.6  406.93    5041  405.69  5046.6  406.02
    5055  405.75  5068.9  407.07  5077.3  408.51  5085.7   411.7  5091.3  414.02
  5099.7  415.03  5108.1   417.4  5113.7   417.9  5130.4   421.6  5144.4  421.88
#Mann= 3 ,-1 , 0
  4732.6     .05       0  4999.6     .03       0  5005.6     .05       0
Bank Sta=4962.6,5085.7
XS Rating Curve= 0 ,0
Exp/Cntr=0.3,0.1

Type RM Length L Ch R = 1 ,19688   ,531,531,531
BEGIN DESCRIPTION:
BATSMITH CREEK 41.0
END DESCRIPTION:
XS GIS Cut Line= 3
      3633349.61     10617310.19      3633449.61     10617010.19
      3633349.62     10616810.22
#Sta/Elev= 30
  4694.6  413.81  4768.4  410.52  4789.5  410.22  4810.6  409.34  4926.5  408.98
  4947.6  407.76  4958.1  405.43  4989.7  401.82  4997.3  399.88    5000  399.38
  5003.3  399.88  5013.6  400.28  5019.2  402.21  5041.6  403.46  5047.2  404.96
  5063.9  405.09  5069.5  406.15  5077.9  406.37  5086.3     407  5091.9  409.41
  5100.3   409.8  5108.7   411.8  5153.4  416.09    5159  416.29  5175.7  418.37
  5189.7  419.17  5212.1  422.37  5220.5   423.1  5231.6  425.24  5234.4  425.24
#Mann= 3 ,-1 , 0
  4694.6     .05       0  4997.3     .03       0  5003.3     .05       0
Bank Sta=4947.6,5077.9
XS Rating Curve= 0 ,0
Exp/Cntr=0.3,0.1

Type RM Length L Ch R = 1 ,19157   ,573,573,573
BEGIN DESCRIPTION:
BATSMITH CREEK 40.0
END DESCRIPTION:
XS GIS Cut Line= 3
      3633949.62     10617260.23      3633849.61     10616960.19
      3633849.61     10616710.16
#Sta/Elev= 30
  4716.2  426.79  4737.3  423.25  4758.4  420.94  4768.9  418.85  4779.5   418.3
  4811.1  413.55    4906  405.01  4916.5  402.59  4927.1  400.99  4969.2  403.96
  4979.8  402.72  4990.3  396.14  4997.8   393.3  5000.6   392.8  5003.8   393.3
  5011.4  397.72  5021.9  398.33  5029.8  401.49    5035  401.49  5042.5  403.24
  5052.5  404.79  5062.5  404.98  5122.5  404.06  5142.5  405.42  5152.5  407.19
  5162.5  407.09  5212.5  413.96  5242.5  420.79  5272.5     424  5282.5  426.18
#Mann= 3 ,-1 , 0
  4716.2     .05       0  4997.8     .03       0  5003.8     .05       0
Bank Sta=4916.5,5042.5
XS Rating Curve= 0 ,0
Exp/Cntr=0.3,0.1

Type RM Length L Ch R = 1 ,18584   ,444,444,444
BEGIN DESCRIPTION:
BATSMITH CREEK 39.0
END DESCRIPTION:
XS GIS Cut Line= 3
      3634462.99     10617032.63      3634265.06     10616803.45
       3633758.1     10616341.63
#Sta/Elev= 30
  4776.5  411.99  4822.9  409.09  4894.2  401.68  4964.7  399.05  4978.7  392.23
    4993  390.29  4997.6  388.17  5000.4  387.67  5003.6  388.17  5007.2  391.05
  5014.9  394.23    5050  396.64  5057.2  398.63  5064.3  399.88  5085.8  400.27
  5269.5   402.1  5326.3  407.78  5361.4  409.32  5411.3  413.17  5418.2  414.79
  5453.3  416.27  5481.7   418.8  5517.5   422.5  5524.3  424.19  5545.9  425.66
  5609.4  434.26  5687.1  438.78  5736.4  443.06  5743.9  444.54  5765.1  444.61
#Mann= 3 ,-1 , 0
  4776.5     .05       0  4997.6     .03       0  5003.6     .05       0
Bank Sta=4964.7,5057.2
XS Rating Curve= 0 ,0
Exp/Cntr=0.3,0.1

Type RM Length L Ch R = 1 ,18140   ,240,240,240
BEGIN DESCRIPTION:
BATSMITH CREEK 38.0
END DESCRIPTION:
XS GIS Cut Line= 3
      3634581.03     10617063.87      3634615.75     10616504.84
      3634452.57     10615886.83
#Sta/Elev= 30
  4627.5  414.21  4731.4  406.31  4881.7  397.04  4941.8  396.06  4981.9  390.13
  4991.9  386.03  4998.9  384.76  5001.7  384.26  5004.9  384.76  5007.4  389.18
  5021.9   386.9    5032   392.2    5052  396.17  5378.6  408.17    5391  410.92
    5420  412.09  5461.2  416.33  5466.4  418.33  5501.5  419.86  5506.7  421.14
  5541.8  421.08  5546.9  423.17    5582   423.6  5587.2  425.23  5616.5  425.68
  5668.2  432.37  5730.2  437.53  5743.1  440.47  5802.6  448.69  5826.8  450.12
#Mann= 3 ,-1 , 0
  4627.5     .05       0  4998.9     .03       0  5004.9     .05       0
Bank Sta=4941.8,5052
XS Rating Curve= 0 ,0
Exp/Cntr=0.3,0.1

Type RM Length L Ch R = 1 ,17900   ,810,810,810
BEGIN DESCRIPTION:
BATSMITH CREEK 37.0
END DESCRIPTION:
XS GIS Cut Line= 3
      3634813.67     10617188.83      3634806.73     10616803.45
      3634796.32     10615964.16
#Sta/Elev= 30
  4562.8  431.06  4621.5  427.59  4661.5  423.94  4701.5  417.07  4741.5  412.29
  4841.5  402.39  4871.5  400.28  4911.5  395.75  4941.5  393.76  4947.4  392.37
  4981.5  388.92  4991.5  384.16  4998.5  383.57  5001.3  383.07  5004.5  383.57
  5011.5  391.44  5021.5  393.57  5031.5  394.41  5191.5  393.79  5271.5  397.81
  5341.5  399.96  5381.5  402.74  5451.5   410.6  5461.5  410.99  5511.5   420.6
  5541.5  424.81  5611.6  429.88  5671.6   437.1  5731.6  441.13  5787.6  442.48
#Mann= 3 ,-1 , 0
  4562.8     .05       0  4998.5     .03       0  5004.5     .05       0
Bank Sta=4941.5,5021.5
XS Rating Curve= 0 ,0
Exp/Cntr=0.3,0.1

Type RM Length L Ch R = 1 ,17090   ,435,435,435
BEGIN DESCRIPTION:
BATSMITH CREEK 36.0
END DESCRIPTION:
XS GIS Cut Line= 3
      3635390.07     10617140.28      3635153.95       10616484.
       3634994.4      10616078.2
#Sta/Elev= 30
  4366.2  427.59  4430.1  422.95  4461.9  422.05  4499.8  418.38  4622.7  414.66
  4709.5  406.98  4734.9  403.33  4759.5  401.43  4765.6  399.78  4770.9  400.44
  4852.4  391.97  4876.4  390.72  4969.9  390.18  4975.2  384.97  4982.7  380.53
  4997.6  378.09  5000.4  377.59  5003.6  378.09  5014.6  382.23  5036.7  386.44
  5056.7  389.99  5153.7  393.71  5278.9  401.71  5284.3  402.94  5325.6  404.83
  5417.1  412.52  5422.4  413.84  5465.3  417.19  5476.6  419.31  5499.7   421.2
#Mann= 3 ,-1 , 0
  4366.2     .05       0  4997.6     .03       0  5003.6     .05       0
Bank Sta=4969.9,5036.7
XS Rating Curve= 0 ,0
Exp/Cntr=0.3,0.1

Type RM Length L Ch R = 1 ,16655   ,503,503,503
BEGIN DESCRIPTION:
BATSMITH CREEK 35.0
END DESCRIPTION:
XS GIS Cut Line= 3
      3635949.58     10616910.16      3635549.61     10616560.19
      3635299.59     10616160.16
#Sta/Elev= 30
  4467.4  440.27  4497.1  436.46  4609.3  421.03  4637.7  415.78  4644.4  412.92
  4665.5  409.93  4672.8   407.3  4701.3  404.51  4715.6  401.05    4800  391.19
  4864.6  387.67  4942.4   387.4    4949  385.52  4956.6  386.26  4963.3  378.01
  4970.9  381.97  4974.5  375.38  4977.3  374.88  4980.5  375.38  5001.8  375.92
  5006.5  378.14  5011.2  376.34  5021.9  381.28    5049  383.14  5064.3  387.06
  5068.7  386.87  5304.9   388.6  5368.6  394.07  5426.3  404.08  5470.6  407.65
#Mann= 7 ,-1 , 0
  4467.4     .05       0  4497.1     .16       0  4665.5     .05       0
  4974.5     .03       0  4980.5     .05       0  5011.2     .16       0
  5068.7     .05       0
Bank Sta=4942.4,5064.3
XS Rating Curve= 0 ,0
Exp/Cntr=0.3,0.1

Type RM Length L Ch R = 1 ,16152   ,439,439,439
BEGIN DESCRIPTION:
BATSMITH CREEK 34.0
END DESCRIPTION:
XS GIS Cut Line= 3
      3636149.62      10616660.2      3635849.61     10616260.19
      3635599.62      10615860.2
#Sta/Elev= 30
    4546  433.31    4596  425.11  4609.6  419.04  4638.7  411.14  4682.5  403.58
  4859.3  386.44  4888.7  384.59  4959.6  384.07  4974.1  374.88  4989.4  373.53
    4993  372.27  4995.8  371.77    4999  372.27  5009.6  373.14    5016  380.72
  5017.9  382.97  5024.1  381.48  5032.5  384.38  5111.4  384.07    5188  384.28
  5211.7  384.75    5245  385.45  5284.8  387.55  5315.1  391.67  5336.7   393.6
  5357.9  400.53  5373.3  397.97  5415.7     404  5482.3   419.5  5517.7  424.15
#Mann= 10 ,-1 , 0
    4546     .16       0  4859.3     .12       0  4989.4     .16       0
    4993     .07       0    4999     .16       0    5016     .12       0
  5111.4     .16       0    5188     .05       0    5245     .16       0
  5315.1     .05       0
Bank Sta=4888.7,5211.7
XS Rating Curve= 0 ,0
Exp/Cntr=0.3,0.1

Type RM Length L Ch R = 1 ,15713   ,450,450,450
BEGIN DESCRIPTION:
BATSMITH CREEK 33.0
END DESCRIPTION:
XS GIS Cut Line= 2
      3636559.03     10616409.12      3635840.66     10615664.72
#Sta/Elev= 30
  4485.4  432.42  4645.7  418.57  4738.7  408.86  4780.3  403.08  4837.8  394.35
  4865.9  392.08  4901.4  388.69  4929.7  382.54  4943.8  380.46  4965.2  380.47
  4972.1  374.84  4987.2  371.62  5004.6  369.18  5007.4  368.68  5010.6  369.18
  5028.7  380.36  5042.9  382.54  5120.8  381.02  5141.9  384.92  5170.2  384.07
  5212.7  378.44    5241  378.91  5262.2  381.74  5309.9  386.87  5354.1  394.94
  5368.3  401.48  5396.6  410.82  5424.9  417.78  5453.2  422.57  5519.9  429.01
#Mann= 9 ,-1 , 0
  4485.4     .16       0  4645.7     .12       0  4738.7     .16       0
  4780.3     .12       0  4865.9     .16       0  4987.2     .12       0
  5004.6     .07       0  5010.6     .12       0  5309.9     .16       0
Bank Sta=4929.7,5262.2
XS Rating Curve= 0 ,0
Exp/Cntr=0.3,0.1

Type RM Length L Ch R = 1 ,15263   ,483,483,483
BEGIN DESCRIPTION:
BATSMITH CREEK 32.0
END DESCRIPTION:
XS GIS Cut Line= 3
       3636649.6     10616110.17      3636499.61     10615710.19
      3636099.58     10615310.16
#Sta/Elev= 30
  4558.8  411.52  4714.5     394  4860.5  380.31  4879.2  378.77  4932.6  379.11
  4940.6  375.92  4945.9  377.11  4970.8  370.85  4987.3  368.44  4997.1  367.04
  4999.9  366.54  5003.1  367.04  5028.4  370.62  5056.7  381.25    5085  380.93
  5100.6  378.04  5212.3  377.94  5226.4  379.73  5233.5   382.3  5240.5  382.92
  5268.8  390.55    5283  392.02  5311.2   397.7  5325.4  402.21  5367.8  410.45
    5382  416.86  5424.4  425.41  5495.1  433.75  5509.2  437.08  5551.7  442.18
#Mann= 5 ,-1 , 0
  4558.8     .16       0  4987.3     .12       0  4997.1     .07       0
  5003.1     .12       0  5100.6     .16       0
Bank Sta=4860.5,5233.5
XS Rating Curve= 0 ,0
Exp/Cntr=0.3,0.1

Type RM Length L Ch R = 1 ,14780   ,618,618,618
BEGIN DESCRIPTION:
BATSMITH CREEK 31.0
END DESCRIPTION:
XS GIS Cut Line= 3
      3636849.61     10616060.21      3636849.61     10615660.19
      3636899.61     10615260.22
#Sta/Elev= 30
  4601.1   408.6  4611.1  405.86  4691.1   392.8  4811.1  379.44  4851.1   376.1
  4911.1  375.63  4921.1  377.28  4942.7  377.27  4961.1  376.65  4971.1  374.69
  4981.1  369.83  4995.6  365.24  4998.4  364.74  5001.6  365.24  5003.6  365.24
  5021.3  375.45  5096.8  375.89  5103.3  376.06  5222.8  376.41  5232.9  376.87
    5243  381.34  5273.2  390.96  5280.8  394.75  5285.8  394.64  5299.7  400.56
  5333.7  411.34  5353.8  414.17    5374  419.43  5398.1  423.65  5404.2  424.13
#Mann= 8 ,-1 , 0
  4601.1     .16       0  4942.7     .12       0  4995.6     .07       0
  5001.6     .12       0  5096.8     .16       0  5103.3     .12       0
  5299.7     .16       0  5398.1     .05       0
Bank Sta=4811.1,5243
XS Rating Curve= 0 ,0
Exp/Cntr=0.3,0.1

Type RM Length L Ch R = 1 ,14162   ,245,245,245
BEGIN DESCRIPTION:
BATSMITH CREEK 30.0
END DESCRIPTION:
XS GIS Cut Line= 3
      3637249.62     10615760.22      3637199.61     10615610.19
       3637149.6     10615210.15
#Sta/Elev= 30
  4849.4   384.5  4881.1  379.23  4923.2  374.85  4944.3  373.74  4965.4  369.65
  4975.9  364.57  4986.5  362.44    4994  362.39  4996.8  361.89    5000  362.39
  5045.3  371.34  5050.4  374.25  5078.1  371.27    5126  375.18  5158.7   378.8
  5168.8  382.79  5178.9  384.71  5210.4  386.62  5244.6  387.05  5279.7  388.91
  5292.2  391.41  5299.8  393.93  5309.9  400.56    5320  403.71    5330   408.5
  5340.1  410.15  5360.3  416.96  5372.9  418.12  5380.4  420.54  5410.7   424.9
#Mann= 5 ,-1 , 0
  4849.4     .12       0    4994     .07       0    5000     .12       0
  5210.4     .16       0  5244.6     .05       0
Bank Sta=4923.2,5126
XS Rating Curve= 0 ,0
Exp/Cntr=0.3,0.1

Type RM Length L Ch R = 1 ,13917   ,354,354,354
BEGIN DESCRIPTION:
BATSMITH CREEK 29.0
END DESCRIPTION:
XS GIS Cut Line= 2
      3637474.41     10615698.78      3637347.89      10615234.3
#Sta/Elev= 30
  4858.5   389.7  4867.4  387.84  4929.1  379.49  4934.4  379.32  4960.7  375.18
  4974.1  371.97  4981.4  371.38  4991.8   364.3  4999.1  360.33  5001.9  359.83
  5005.1  360.33  5008.6  361.55  5013.8  361.95  5022.9  365.59  5033.2  371.06
  5043.2  372.47  5074.7  371.96  5088.1  372.59  5116.1   370.3  5147.2  372.59
  5162.5  373.04    5168  374.34  5202.2  377.62  5209.4  379.55  5245.3  383.19
  5276.5  385.77    5282  387.21  5302.7  388.33  5323.4  391.57  5339.9  393.03
#Mann= 5 ,-1 , 0
  4858.5     .16       0  4934.4     .12       0  4999.1     .07       0
  5005.1     .12       0  5245.3     .16       0
Bank Sta=4974.1,5147.2
XS Rating Curve= 0 ,0
Exp/Cntr=0.3,0.1

Type RM Length L Ch R = 1 ,13563   ,96,96,96
BEGIN DESCRIPTION:
Mapping XS ecd5a18d
END DESCRIPTION:
XS GIS Cut Line= 3
      3637576.83     10615596.28      3637583.77     10615408.81
      3637531.89     10615094.06
#Sta/Elev= 30
  4753.9  383.12    4760  381.22    4790  377.44    4810  376.09    4830  371.61
  4840.1  370.77  4850.1  372.17  4870.1  363.55  4880.1  363.19  4890.1   365.9
  4900.1  365.82  4910.1  368.34  4920.1  369.32    4943  367.91  4970.5  366.37
  4998.9  358.72  5001.7  358.22  5004.9  358.72  5021.2   368.5  5041.5   371.2
  5051.6  371.59  5063.1   374.6  5112.4  381.94  5132.7  385.53  5138.1  387.74
  5152.9  391.97  5163.1  397.21  5173.2  400.31  5180.3  404.59  5260.5  420.74
#Mann= 5 ,-1 , 0
  4753.9     .05       0    4943     .12       0  4998.9     .07       0
  5004.9     .12       0  5138.1     .16       0
Bank Sta=4850.1,5041.5
XS Rating Curve= 0 ,0
Exp/Cntr=0.3,0.1

Type RM Length L Ch R = 1 ,13467   ,165,165,165
BEGIN DESCRIPTION:
BATSMITH CREEK 28.0
END DESCRIPTION:
XS GIS Cut Line= 4
      3637602.86     10615606.77      3637649.74     10615332.42
      3637651.48     10615256.03      3637628.96     10614954.61
#Sta/Elev= 30
  4688.5  382.75  4699.6  383.72  4715.5  380.38  4754.6  376.88  4759.7  378.53
  4796.6   375.6  4879.9  373.33  4908.2  370.92    4935  363.78    4940     364
  4955.9  358.02  4958.7  357.52  4961.9  358.02  4989.1  362.57  5003.7  362.07
  5019.1  361.74  5029.1  364.33  5043.2  364.88  5049.1  369.73  5059.1  372.18
  5069.1  373.11  5099.2  380.91  5109.3  380.54  5129.3  384.07  5139.9  389.08
  5219.6  409.03  5267.2  414.14  5272.2  416.74  5299.8  421.73  5345.5   424.4
#Mann= 4 ,-1 , 0
  4688.5     .05       0  4955.9     .04       0  4961.9     .05       0
  5003.7     .16       0
Bank Sta=4908.2,5059.1
XS Rating Curve= 0 ,0
Exp/Cntr=0.3,0.1

Type RM Length L Ch R = 1 ,13302   ,66,66,66
BEGIN DESCRIPTION:
Mapping XS 660ea902
END DESCRIPTION:
XS GIS Cut Line= 3
      3637689.67     10615629.32      3637802.52      10615210.9
      3637707.04     10614959.17
#Sta/Elev= 30
    4649  386.48  4745.6  382.49  4865.6  371.75  4886.3     368  4894.9  363.21
  4900.1  365.23    4907  362.59  4917.4  367.61  4927.7  369.29  4969.2  366.72
  4974.8  360.19  4989.5  358.32  4997.2  358.03    5000  357.53  5003.2  358.03
  5009.5  364.22  5014.7  364.37  5021.8  370.54  5072.8  370.42  5095.1  370.49
  5101.9  370.46  5107.3  373.63  5132.1  372.13    5187  378.11  5199.2   381.2
  5241.9  387.63  5254.3  393.48  5286.3  400.94  5318.4   412.5  5351.6  417.53
#Mann= 7 ,-1 , 0
    4649     .05       0  4989.5     .08       0  4997.2     .07       0
  5003.2     .08       0  5021.8     .12       0  5095.1     .05       0
  5199.2     .16       0
Bank Sta=4865.6,5072.8
XS Rating Curve= 0 ,0
Exp/Cntr=0.3,0.1

Type RM Length L Ch R = 1 ,13236   ,446,446,446
BEGIN DESCRIPTION:
Mapping XS 4f970281
END DESCRIPTION:
XS GIS Cut Line= 3
      3637835.51     10615615.42      3637837.24     10615144.92
      3637762.59     10614948.74
#Sta/Elev= 30
  4710.6  398.49  4785.8  394.56  4825.8   390.4  4885.8  382.24  4915.8  374.94
  4925.1  374.08  4945.8   371.4  4965.8  365.93  4975.8  361.05  4985.8  357.98
  4992.8  357.31  4995.6  356.81  4998.8  357.31  5015.8  359.27  5025.8  363.34
  5045.8  368.64  5065.8  369.43  5115.8   368.1  5144.8  369.43  5155.8  369.84
  5184.8   371.3    5190  373.41  5214.8     373    5229  374.31  5269.6  379.59
  5285.1  383.17  5293.2  383.74  5314.6  388.75  5346.7  402.12    5391  411.39
#Mann= 6 ,-1 , 0
  4710.6     .05       0  4925.1     .12       0  4992.8     .07       0
  4998.8     .12       0  5144.8     .05       0  5285.1     .16       0
Bank Sta=4945.8,5155.8
XS Rating Curve= 0 ,0
Exp/Cntr=0.3,0.1

Type RM Length L Ch R = 1 ,12790   ,423,423,423
BEGIN DESCRIPTION:
BATSMITH CREEK 27.0
END DESCRIPTION:
XS GIS Cut Line= 3
      3638299.59     10615210.17      3638149.61     10615110.19
      3637749.58     10614910.17
#Sta/Elev= 30
  4805.9  379.27  4819.4  375.25  4841.9  371.81  4885.5  368.39    4914  367.33
  4921.5  363.61  4927.6  362.36  4950.1     360  4988.9  358.03  4997.1  354.37
  4999.9  353.87  5003.1  354.37  5008.5  355.69  5016.9  366.22    5084   367.7
  5168.3  370.12  5201.4  371.11  5232.1  375.47  5246.1  374.83  5299.2  386.68
  5310.1  391.16  5321.6  392.88  5329.9  396.15  5343.9     398  5352.3  401.64
  5366.3  403.34  5374.7  406.45  5380.3  405.59    5397  409.68  5433.4  414.48
#Mann= 5 ,-1 , 0
  4805.9     .12       0  4997.1     .07       0  5003.1     .12       0
  5168.3     .05       0  5310.1     .16       0
Bank Sta=4885.5,5084
XS Rating Curve= 0 ,0
Exp/Cntr=0.3,0.1

Type RM Length L Ch R = 1 ,12367   ,461,461,461
BEGIN DESCRIPTION:
BATSMITH CREEK 26.0
END DESCRIPTION:
XS GIS Cut Line= 3
      3638499.61      10615210.2      3638399.61     10614860.19
       3638099.6     10614560.18
#Sta/Elev= 30
  4638.6  385.67  4669.8  381.91  4680.2  377.17  4689.3  376.08  4694.5  378.44
    4701  376.21  4733.5     374  4784.2  365.46  4834.9  363.16  4870.2  363.98
  4912.9  363.87  4946.7  360.19  4971.4  361.47  4980.5  359.73  4992.2  352.88
    4997  352.37  4999.8  351.87    5003  352.37  5016.8  355.03  5030.9   360.6
  5059.2  364.58    5144  363.29  5186.5  369.15  5313.7   396.9    5342  404.93
  5356.2   407.4  5370.3  412.86  5384.5  414.55  5398.6  420.17  5426.9  426.02
#Mann= 4 ,-1 , 0
  4638.6     .12       0  4870.2     .16       0    4997     .07       0
    5003     .16       0
Bank Sta=4912.9,5059.2
XS Rating Curve= 0 ,0
Exp/Cntr=0.3,0.1

Type RM Length L Ch R = 1 ,11906   ,341,341,341
BEGIN DESCRIPTION:
BATSMITH CREEK 25.0
END DESCRIPTION:
XS GIS Cut Line= 3
      3638949.59     10614910.16      3638799.61     10614710.19
      3638399.58     10614410.17
#Sta/Elev= 30
  4768.2  380.26  4846.3  368.07  4868.2     363  4875.5  355.75    4890  354.02
  4896.3  354.68  4910.9  352.62  4925.5   352.9  4931.7  355.25  4946.3  356.42
  4954.6  353.72  4968.2  356.64  4981.7  352.74  4993.3  350.91    4996  350.41
  4999.3  350.91  5004.6  352.84  5010.9  352.17    5015  356.69  5025.5  357.18
  5031.7  359.32  5110.9  358.91  5225.5  360.61  5365.8  364.06  5418.2  367.05
  5468.2  375.15  5475.5  379.13  5481.7  379.23  5504.6  385.39  5518.2  386.42
#Mann= 4 ,-1 , 0
  4768.2     .12       0  4993.3     .07       0  4999.3     .12       0
  5365.8     .16       0
Bank Sta=4868.2,5225.5
XS Rating Curve= 0 ,0
Exp/Cntr=0.3,0.1

Type RM Length L Ch R = 1 ,11565   ,628,628,628
BEGIN DESCRIPTION:
BATSMITH CREEK 24.0
END DESCRIPTION:
XS GIS Cut Line= 2
       3639293.4     10614924.75      3638730.91     10614127.88
#Sta/Elev= 30
  4664.7  389.18    4689  388.49  4749.6  385.26  4814.9  377.61    4901   364.8
  4928.1  364.62    4964  360.11  4978.6  354.05  4993.4  352.36  4997.8  349.51
  5000.5  349.01  5003.8  349.51  5022.9  351.18  5029.1  349.58    5050  350.04
  5058.6  357.56  5064.8  353.53  5071.7  355.09  5079.6  357.45  5100.5  357.91
  5266.7  357.11  5317.2  357.89  5338.1  359.92  5369.4  363.19  5475.1  380.18
  5495.7  383.41  5546.2  384.87  5581.9  389.31  5596.7  388.88  5640.1  392.31
#Mann= 7 ,-1 , 0
  4664.7     .12       0    4689     .16       0  4997.8     .07       0
  5003.8     .16       0  5071.7     .12       0  5369.4     .16       0
  5475.1     .12       0
Bank Sta=4964,5338.1
XS Rating Curve= 0 ,0
Exp/Cntr=0.3,0.1

Type RM Length L Ch R = 1 ,10937   ,337,337,337
BEGIN DESCRIPTION:
BATSMITH CREEK 23.0
END DESCRIPTION:
XS GIS Cut Line= 3
      3639547.32     10615143.88      3639595.47     10614518.48
      3639079.85      10613721.6
#Sta/Elev= 30
  4491.9  396.36  4505.6  395.79  4555.8  395.59  4595.9  392.52  4605.9  393.67
  4676.1  391.19  4750.8  386.63  4774.2  384.43  4876.7  373.78  4926.9  363.52
  4936.9  363.21    4967  357.34  4974.8  356.19  4979.8   349.6  4984.1  345.97
  4986.8  345.47  4990.1  345.97  5007.1  349.26  5017.1   354.5  5128.1  354.82
  5149.2  354.41  5209.6  355.37  5533.5  354.19  5582.9  353.99  5629.3  354.29
  5700.7   357.2  5903.2  370.68  6001.3  375.92  6055.8  378.38  6068.3  380.02
#Mann= 11 ,-1 , 0
  4491.9     .16       0  4505.6     .12       0  4750.8     .16       0
  4774.2     .12       0  4984.1     .07       0  4990.1     .12       0
  5128.1     .16       0  5149.2     .12       0  5533.5     .16       0
  5582.9     .12       0  6001.3     .16       0
Bank Sta=4967,5700.7
XS Rating Curve= 0 ,0
Exp/Cntr=0.3,0.1

Type RM Length L Ch R = 1 ,10600   ,638,638,638
BEGIN DESCRIPTION:
BATSMITH CREEK 22.0
END DESCRIPTION:
XS GIS Cut Line= 3
       3640137.6     10614984.15       3639800.8     10614595.26
      3639380.85     10613654.72
#Sta/Elev= 30
  4413.2  396.43  4619.9  373.65  4697.8  366.94  4804.2  356.24    4882   355.2
  4918.2  352.43  4927.7   353.4  4969.5  351.35    4977  350.65  4987.2  345.74
  4992.7  347.71  4995.9  344.96  4998.7  344.46  5001.9  344.96  5009.9  352.05
  5015.9  353.25  5021.4  350.84  5062.3  354.35  5109.7  352.84  5286.4  353.29
  5349.4  352.11  5432.5  354.43  5447.9  352.82  5530.8  356.01  5597.2  360.68
  5657.8  365.94  5688.9  371.33  5743.6  376.72  5929.8  381.16  5957.7  383.19
#Mann= 7 ,-1 , 0
  4413.2     .16       0  4697.8     .12       0  4995.9     .07       0
  5001.9     .12       0  5109.7     .16       0  5286.4     .12       0
  5597.2     .16       0
Bank Sta=4804.2,5530.8
XS Rating Curve= 0 ,0
Exp/Cntr=0.3,0.1

Type RM Length L Ch R = 1 ,9962    ,532,532,532
BEGIN DESCRIPTION:
BATSMITH CREEK 21.0
END DESCRIPTION:
XS GIS Cut Line= 3
      3640475.71     10614409.12      3639944.43     10614070.56
      3639611.08     10613580.95
#Sta/Elev= 30
  4568.5  389.84  4630.4  388.33  4739.6  381.06  4775.9  375.07  4781.9  371.77
  4818.3  369.21  4854.7  363.51  4875.8  361.96  4933.4  354.21  4948.6  353.49
  4969.8  352.27    4985  347.02  4990.9  346.57  4997.2  342.84    5000  342.34
  5003.2  342.84  5021.4  349.62  5027.3  349.88  5151.8  351.55  5216.5  350.56
  5295.1  351.42  5324.3  349.97  5385.8  352.52  5396.1  352.03  5404.6  353.58
  5421.2  354.62  5446.9  355.23  5554.7  364.13  5728.2  372.38  5790.8  377.89
#Mann= 6 ,-1 , 0
  4568.5     .12       0  4997.2     .07       0  5003.2     .12       0
  5295.1     .16       0  5385.8     .12       0  5421.2     .16       0
Bank Sta=4948.6,5404.6
XS Rating Curve= 0 ,0
Exp/Cntr=0.3,0.1

Type RM Length L Ch R = 1 ,9430    ,396,396,396
BEGIN DESCRIPTION:
BATSMITH CREEK 20.0
END DESCRIPTION:
XS GIS Cut Line= 2
      3640601.62     10613921.01      3639939.13     10613544.31
#Sta/Elev= 30
  4669.8  369.26  4787.8  354.02  4819.6  351.49  4874.9  348.95  4971.2  348.91
    4981   347.9  4986.8   344.3  4994.2  341.99  5005.4  341.82  5008.1  341.32
  5011.4  341.82  5017.2  347.56  5024.2  348.33  5067.5  347.02    5105   348.6
  5148.2  346.76  5201.3  347.13  5235.8  351.33  5268.5  356.89  5303.9  360.51
  5309.6   363.8  5316.3   364.9  5347.1  367.13  5352.9  370.14  5384.6  370.99
  5390.4  373.64  5406.2  372.63    5412  373.68  5427.9  371.55  5431.9  373.86
#Mann= 5 ,-1 , 0
  4669.8     .16       0  4874.9     .12       0  5005.4     .07       0
  5011.4     .12       0  5268.5     .05       0
Bank Sta=4819.6,5235.8
XS Rating Curve= 0 ,0
Exp/Cntr=0.3,0.1

Type RM Length L Ch R = 1 ,9034    ,437,437,437
BEGIN DESCRIPTION:
BATSMITH CREEK 19.0
END DESCRIPTION:
XS GIS Cut Line= 3
      3640849.61     10613810.19      3640499.61     10613410.19
      3640099.62     10613260.19
#Sta/Elev= 30
  4466.3  382.61  4522.8  376.57    4537  372.72  4567.3  367.45  4665.1  353.78
  4700.3  350.64  4757.2  345.44  4814.7  346.72  4884.4   345.9  4976.5  347.77
    4984  346.68  4990.7  340.95  4996.5  340.79  5004.6  340.53  5007.4  340.03
  5010.6  340.53  5012.9  341.35  5019.2  347.52  5085.5  346.39  5158.9  345.53
  5208.7  350.66  5211.2   351.3  5254.1  357.37  5269.3  358.18  5324.4  366.31
  5349.4  370.52  5360.9  376.18    5385  380.02  5409.9  381.71    5425  381.07
#Mann= 8 ,-1 , 0
  4466.3     .16       0  4567.3     .05       0  4814.7     .12       0
  4996.5     .16       0  5004.6     .07       0  5010.6     .16       0
  5085.5     .12       0  5211.2     .16       0
Bank Sta=4700.3,5208.7
XS Rating Curve= 0 ,0
Exp/Cntr=0.3,0.1

Type RM Length L Ch R = 1 ,8597    ,389,389,389
BEGIN DESCRIPTION:
BATSMITH CREEK 18.0
END DESCRIPTION:
XS GIS Cut Line= 3
      3640972.19      10613741.8      3640843.73     10613137.67
      3640843.73     10612653.41
#Sta/Elev= 30
    4448  373.12  4479.8  370.57  4484.9  371.83  4521.2   365.9  4534.5  365.92
  4556.5  361.63  4613.2  355.82  4693.6  352.05  4766.6  349.56  4889.3  344.26
  4981.3  346.14  4991.5  340.56  4998.7  339.76  5001.5  339.26  5004.7  339.76
  5010.1  339.87  5015.2  345.02  5022.2  346.13  5059.7  344.15  5073.1  346.47
  5103.1  346.93  5113.1  342.84  5123.1  341.03  5133.1  346.52  5173.1   345.4
  5223.1  350.19  5293.1  356.51  5482.8  378.46  5522.9  382.37  5549.9  385.85
#Mann= 7 ,-1 , 0
    4448     .16       0  4556.5     .05       0  4693.6     .12       0
  4998.7     .07       0  5004.7     .12       0  5482.8     .16       0
  5522.9     .12       0
Bank Sta=4766.6,5223.1
XS Rating Curve= 0 ,0
Exp/Cntr=0.3,0.1

Type RM Length L Ch R = 1 ,8208    ,672,672,672
BEGIN DESCRIPTION:
BATSMITH CREEK 17.0
END DESCRIPTION:
XS GIS Cut Line= 2
      3641230.89     10613690.38      3641137.19     10612654.51
#Sta/Elev= 30
  4357.5  384.46  4417.9  384.07  4478.2  380.86    4549  372.87  4638.8  356.21
  4659.1  354.03  4699.1  349.58  4757.3  343.13  4839.6  342.49  4983.8  345.06
  4990.3  339.84  4997.3  339.06  5000.1  338.56  5003.3  339.06  5010.3     340
  5020.4   344.3  5050.5  344.21  5089.5  348.67  5094.5  347.75  5100.7  349.63
  5150.9  356.22    5181  365.39  5200.2  369.53  5205.2  368.98  5211.2  372.09
  5231.2  376.17  5267.1  380.18  5310.9  386.11  5351.7  386.57  5397.6  384.24
#Mann= 6 ,-1 , 0
  4357.5     .16       0    4549     .05       0  4659.1     .12       0
  4997.3     .07       0  5003.3     .12       0  5267.1     .16       0
Bank Sta=4699.1,5100.7
XS Rating Curve= 0 ,0
Exp/Cntr=0.3,0.1

Type RM Length L Ch R = 1 ,7536    ,295,295,295
BEGIN DESCRIPTION:
BATSMITH CREEK 16.0
END DESCRIPTION:
XS GIS Cut Line= 3
      3641599.61     10613560.19      3641649.61     10613260.19
      3641499.62     10612860.22
#Sta/Elev= 30
  4666.2  374.77  4747.3  363.93    4760   363.4  4808.1  355.73  4821.8  354.89
  4881.6  346.75  4929.8  341.99    4973  342.65  4980.1  339.85  4985.5   342.4
  4999.4   336.2  5002.1   335.7  5005.4   336.2  5015.7  336.89  5023.7  341.76
  5034.4  343.03  5141.2  343.61  5173.3  341.77  5194.6  342.81  5211.5  345.78
  5241.8  349.93    5248   353.1  5258.7  354.98  5266.7  359.76  5280.1  362.93
  5290.7  367.32  5312.1  372.02  5344.1  376.23  5365.5  380.91  5397.5  382.47
#Mann= 4 ,-1 , 0
  4666.2     .05       0  4821.8     .12       0  4999.4     .07       0
  5005.4     .12       0
Bank Sta=4881.6,5211.5
XS Rating Curve= 0 ,0
Exp/Cntr=0.3,0.1

Type RM Length L Ch R = 1 ,7241    ,523,523,523
BEGIN DESCRIPTION:
BATSMITH CREEK 15.0
END DESCRIPTION:
XS GIS Cut Line= 2
      3641870.38     10613569.91      3642031.84     10612710.55
#Sta/Elev= 30
  4705.3   358.3  4751.1  353.51  4847.5  345.47    4892  343.24    4939  340.35
  4989.9  341.23    4997  335.68  4999.1  335.53  5001.8  335.03  5005.1  335.53
  5010.3   335.8  5020.4   341.6  5132.4  339.75  5173.1  340.02  5183.2  340.95
  5244.3     339  5264.6  339.67  5295.2  338.17  5379.9  340.53  5427.3  344.19
  5432.4  344.02  5468.1   349.5  5508.8  357.09    5519  360.51  5529.2  362.06
  5537.4  366.17  5549.5  368.23  5559.7  372.11  5569.9  373.16  5579.7  375.62
#Mann= 4 ,-1 , 0
  4705.3     .16       0  4751.1     .12       0  4999.1     .07       0
  5005.1     .12       0
Bank Sta=4892,5427.3
XS Rating Curve= 0 ,0
Exp/Cntr=0.3,0.1

Type RM Length L Ch R = 1 ,6718    ,579,579,579
BEGIN DESCRIPTION:
BATSMITH CREEK 14.0
END DESCRIPTION:
XS GIS Cut Line= 3
      3641755.82     10614319.88      3642333.41     10613216.76
      3642230.01     10612633.84
#Sta/Elev= 30
  3561.2  394.73  3645.2  389.55  3727.8  389.79  3733.4     388  3771.9  389.37
  3816.1  388.47  3821.7  386.77  3948.5  387.41  3986.9  389.39  4068.8  388.04
  4157.8  380.79  4319.3   361.1    4366  356.62  4510.9  340.45  4527.3  338.22
  4955.2  337.31  4965.4  336.98  4970.9  334.67    4976  336.21    5003  330.75
  5005.8  330.25    5009  330.75  5024.9  336.49  5097.4   334.6    5138  342.38
  5197.1  357.14  5209.1  357.53  5256.2  370.31    5331  378.97  5398.4  379.58
#Mann= 5 ,-1 , 0
  3561.2     .16       0  4319.3     .05       0    4366     .12       0
    5003     .07       0    5009     .12       0
Bank Sta=4510.9,5138
XS Rating Curve= 0 ,0
Exp/Cntr=0.3,0.1

Type RM Length L Ch R = 1 ,6139    ,528,528,528
BEGIN DESCRIPTION:
BATSMITH CREEK 13.0
END DESCRIPTION:
XS GIS Cut Line= 3
       3643323.5     10614095.94      3642750.59     10613273.04
      3642512.54     10612634.14
#Sta/Elev= 30
  3854.1  407.18  3996.7  404.83  4101.4  394.28  4169.5  385.54  4276.8   379.7
  4306.5  380.37  4312.6  378.09  4408.4  371.01  4472.9  362.16    4591  349.53
  4622.4  344.88  4699.2  339.42  4759.5  336.18    4831  333.38  4977.2  333.19
  4985.5  331.21  4987.9  324.65  4990.6  324.15  4993.9  324.65  5009.2  326.13
  5015.9   333.2  5021.2  333.46  5233.3  332.47  5333.4  336.04  5346.9  337.11
  5413.8  348.01  5457.4  360.01  5470.5   361.5  5499.4  369.74  5538.6  371.87
#Mann= 10 ,-1 , 0
  3854.1     .16       0  4101.4     .05       0  4408.4     .16       0
  4472.9     .05       0    4591     .16       0  4699.2     .12       0
  4987.9     .07       0  4993.9     .12       0  5346.9     .16       0
  5470.5     .05       0
Bank Sta=4759.5,5333.4
XS Rating Curve= 0 ,0
Exp/Cntr=0.3,0.1

Type RM Length L Ch R = 1 ,5611    ,255,255,255
BEGIN DESCRIPTION:
BATSMITH CREEK 12.0
END DESCRIPTION:
XS GIS Cut Line= 3
      3643149.61      10613210.2      3642999.61     10612810.19
      3642899.61     10612460.21
#Sta/Elev= 30
    4597  360.08  4612.1  359.02  4618.4     357    4671  348.97  4714.5  343.23
  4722.5  340.92  4746.5  337.66  4758.1  334.13  4767.9  331.25  4777.7  330.92
  4821.3  331.82  4923.6  329.67  4978.8  330.23  4984.2   328.9  4992.2  323.44
  4999.9  320.64  5002.6  320.14  5005.9  320.64  5009.1  322.48  5014.4  328.41
  5021.5  329.34  5128.2  329.32  5159.4  332.91  5180.2  334.75  5186.7  336.64
    5201  337.62  5264.7  347.36  5325.8  361.69  5332.3   364.6  5388.2  370.77
#Mann= 4 ,-1 , 0
    4597     .16       0    4671     .12       0  4999.9     .07       0
  5005.9     .12       0
Bank Sta=4758.1,5159.4
XS Rating Curve= 0 ,0
Exp/Cntr=0.3,0.1

Type RM Length L Ch R = 1 ,5356    ,538,538,538
BEGIN DESCRIPTION:
BATSMITH CREEK 11.0
END DESCRIPTION:
XS GIS Cut Line= 3
      3643415.77     10613089.59      3643047.47     10612356.37
      3642526.65     10611840.76
#Sta/Elev= 30
  4581.8  348.51  4614.7  342.84  4652.5  339.47  4691.6  332.27  4697.2  333.96
    4708  330.79  4838.5   328.1  4981.9  328.27  4995.2  323.63  5001.2  319.62
    5004  319.12  5007.2  319.62  5026.6  328.68  5099.1   327.2  5138.2  331.55
  5241.4   352.7  5300.1  360.06  5331.7  360.44  5419.3  354.52  5574.9  354.38
  5603.2   355.9  5645.6  361.85  5680.9  363.44  5758.7  372.95  5794.1  374.54
  5801.2  376.49  5822.4  376.38  5914.3  386.62  6013.3  393.53  6135.2  399.33
#Mann= 5 ,-1 , 0
  4581.8     .16       0    4708     .12       0  5001.2     .07       0
  5007.2     .12       0  5331.7     .16       0
Bank Sta=4697.2,5138.2
XS Rating Curve= 0 ,0
Exp/Cntr=0.3,0.1

Type RM Length L Ch R = 1 ,4818    ,588,588,588
BEGIN DESCRIPTION:
BATSMITH CREEK 10.0
END DESCRIPTION:
XS GIS Cut Line= 3
      3643792.25     10613158.42      3643594.34     10612106.37
      3643682.69     10611373.58
#Sta/Elev= 30
  4288.8  354.86  4331.5  347.43  4337.9  343.69  4374.9  340.03    4494  329.45
    4521  327.11  4948.4  325.79  4968.7  322.54  4981.6  325.86  4996.3  317.99
    4999  317.49  5002.3  317.99  5009.5  318.69  5019.6  326.58  5060.3  330.82
  5119.8  341.65  5191.6  355.12  5249.1  362.46  5294.4  364.83  5443.1  353.53
  5597.2  347.91  5687.8   348.4  5743.6  352.46  5838.9  363.59  5919.5  377.95
  5972.6  384.35  6020.2  388.78  6032.6  386.08  6080.7  386.88  6097.4  389.41
#Mann= 7 ,-1 , 0
  4288.8     .16       0  4374.9     .12       0  4996.3     .07       0
  5002.3     .12       0  5119.8     .16       0  5743.6     .12       0
  5972.6     .16       0
Bank Sta=4494,5060.3
XS Rating Curve= 0 ,0
Exp/Cntr=0.3,0.1

Type RM Length L Ch R = 1 ,4230    ,447,447,447
BEGIN DESCRIPTION:
BATSMITH CREEK 9.0
END DESCRIPTION:
XS GIS Cut Line= 3
      3644149.61     10612910.18      3644199.61     10612510.19
      3643849.62      10612110.2
#Sta/Elev= 30
  4629.7  351.23  4706.6  342.03  4748.1  335.14  4753.1  335.86  4760.7  333.68
  4821.2  326.65  4851.4  323.57  4972.3  322.76  4982.4  321.63    4990  318.41
    4992  315.14  4994.8  314.64    4998  315.14  5002.6  317.52  5022.7  321.75
  5036.1  321.77  5039.9  324.26  5046.6  322.62  5054.2  324.48  5096.9  323.41
  5103.5  319.99  5117.7  323.63  5152.9  324.14  5181.3  322.58  5245.4  323.85
  5273.4  322.59  5337.9  325.39    5442  332.84    5458  333.48  5564.3  347.12
#Mann= 5 ,-1 , 0
  4629.7     .16       0  4706.6     .12       0    4992     .07       0
    4998     .12       0    5442     .16       0
Bank Sta=4821.2,5337.9
XS Rating Curve= 0 ,0
Exp/Cntr=0.3,0.1

Type RM Length L Ch R = 1 ,3783    ,448,448,448
BEGIN DESCRIPTION:
BATSMITH CREEK 8.0
END DESCRIPTION:
XS GIS Cut Line= 3
      3644380.81     10613168.86      3644620.38     10612517.83
       3644630.8      10611585.5
#Sta/Elev= 30
  4241.6  353.69  4340.4  345.47  4389.4  343.37  4613.1  323.14  4659.5  318.47
  4762.3  320.71  4868.9  319.65    4983  320.74    4993  318.28    5000  313.99
  5002.7  313.49    5006  313.99    5013  320.13    5033  320.41    5043  318.64
    5053  321.84    5293  318.91    5373  319.98    5393  322.44    5503  334.98
    5583  350.28    5603  356.16  5612.3  356.81    5633  358.35    5653  356.97
    5673  357.62    5693  359.53    5713  358.73    5793  349.56  5867.7  344.74
#Mann= 4 ,-1 , 0
  4241.6     .12       0    5000     .07       0    5006     .12       0
  5612.3      .1       0
Bank Sta=4613.1,5393
XS Rating Curve= 0 ,0
Exp/Cntr=0.3,0.1

Type RM Length L Ch R = 1 ,3335    ,280,280,280
BEGIN DESCRIPTION:
Mapping XS 43ef6bcb
END DESCRIPTION:
XS GIS Cut Line= 3
      3644665.47     10613355.25      3644957.12     10612579.25
      3645248.57     10611564.37
#Sta/Elev= 30
  4123.1   362.4    4177  356.66    4246  353.24  4319.1  344.83  4372.7  343.12
  4408.3  337.79  4573.6  321.99  4609.2  316.74  4628.8  318.53    4940   318.2
  4948.9  315.92  4978.2  317.08  4992.7  313.43  5008.9  312.81  5011.6  312.31
  5014.9  312.81  5017.1  317.31  5023.9  318.06  5084.5  314.49  5089.7  316.57
  5107.2  314.66  5157.2  317.56    5274  315.64  5398.5  321.84  5432.6  323.24
  5688.4  335.92  5816.2  342.42  5956.3  345.06  6001.3     349    6008  349.76
#Mann= 7 ,-1 , 0
  4123.1     .16       0  4319.1     .12       0  5008.9     .07       0
  5014.9     .12       0  5432.6     .16       0  5688.4      .1       0
  6001.3     .07       0
Bank Sta=4573.6,5398.5
XS Rating Curve= 0 ,0
Exp/Cntr=0.3,0.1

Type RM Length L Ch R = 1 ,3055    ,250,250,250
BEGIN DESCRIPTION:
BATSMITH CREEK 7.0
END DESCRIPTION:
XS GIS Cut Line= 2
      3644816.49     10613368.32      3645477.97     10611920.36
#Sta/Elev= 30
  4349.9  364.56  4508.8  355.15  4562.1  350.79  4567.7  344.58  4578.7  342.29
  4585.1  336.09  4608.1  329.09  4751.8  321.58  4819.4  320.07    4901  315.59
    4970  316.97  4990.1  310.46  4992.8  309.96  4996.1  310.46  5021.6  316.63
  5136.7     323  5142.2  320.67  5179.1   321.3  5271.3  321.62  5384.2  324.46
  5469.2  326.75  5532.5  332.77  5619.3   341.1  5624.8  344.54  5665.3  344.81
  5693.8  348.76  5716.9  346.17  5814.5  349.84  5858.5  348.33  5941.8  352.28
#Mann= 9 ,-1 , 0
  4349.9     .16       0  4508.8     .05       0  4819.4     .12       0
  4990.1     .07       0  4996.1     .12       0  5179.1     .05       0
  5384.2     .08       0  5532.5     .05       0  5858.5      .1       0
Bank Sta=4751.8,5271.3
XS Rating Curve= 0 ,0
Exp/Cntr=0.3,0.1

Type RM Length L Ch R = 1 ,2805    ,154,154,154
BEGIN DESCRIPTION:
BATSMITH CREEK 6.0
END DESCRIPTION:
XS GIS Cut Line= 2
       3645063.9     10613446.42      3645644.62     10612050.61
#Sta/Elev= 30
  4306.9  362.58  4313.9  359.99  4356.2  363.56  4400.3  360.73  4414.7  357.89
  4467.8  356.55  4508.6  353.03  4536.6  346.76  4634.7  337.46  4725.1  325.25
  4790.2  320.24  4881.9  315.75  4974.3  315.62    4993  309.03  4995.8  308.53
    4999  309.03  5006.5  314.06  5017.7  316.24  5050.2   315.4  5104.3  319.82
    5236  327.07  5364.3  341.42  5385.9  346.23  5449.8  351.09  5494.2  362.35
  5556.1  373.39  5677.8  374.66  5732.5  371.05  5744.7  367.76  5818.7  364.28
#Mann= 8 ,-1 , 0
  4306.9     .16       0  4536.6     .05       0  4634.7     .16       0
  4725.1     .12       0    4993     .07       0    4999     .12       0
    5236     .05       0  5677.8     .16       0
Bank Sta=4790.2,5104.3
XS Rating Curve= 0 ,0
Exp/Cntr=0.3,0.1

Type RM Length L Ch R = 1 ,2651    ,340,340,340
BEGIN DESCRIPTION:
Mapping XS 402dd50c
END DESCRIPTION:
XS GIS Cut Line= 2
      3645225.36     10613527.15      3645766.67     10612054.16
#Sta/Elev= 30
  4257.5  366.68  4313.1  361.77    4374  362.86  4435.4  359.88  4454.8  355.23
  4460.1  357.37  4490.6  352.77  4515.8  346.44  4531.3  347.18  4656.4  330.89
  4774.1  319.31    4835  313.95  4968.1  315.67  4982.1  314.25  4986.4  309.99
  4989.1  309.49  4992.4  309.99  5012.5  315.82  5068.2  314.02  5123.8  319.32
  5277.9   335.7  5331.8  339.08    5357  345.35  5417.9  348.94  5498.7  360.05
  5534.5  357.54  5584.8  362.07  5611.3  359.34  5737.2  356.73  5826.8   360.5
#Mann= 6 ,-1 , 0
  4257.5     .16       0  4656.4     .12       0  4986.4     .07       0
  4992.4     .12       0  5277.9     .05       0  5611.3     .16       0
Bank Sta=4774.1,5123.8
XS Rating Curve= 0 ,0
Exp/Cntr=0.3,0.1

Type RM Length L Ch R = 1 ,2311    ,416,416,416
BEGIN DESCRIPTION:
BATSMITH CREEK 5.0
END DESCRIPTION:
XS GIS Cut Line= 3
       3645549.6     10613410.21      3645749.61     10613010.19
      3645949.61     10612760.18
#Sta/Elev= 30
  4523.5  355.89  4526.3  355.89  4531.9  352.79  4554.3  348.24  4568.2  346.59
  4576.6  343.99  4635.3  333.09  4659.5  329.78    4694  325.74  4702.4  323.88
  4761.1  317.53  4777.9  314.69  4800.2  312.87  4836.6  311.38    4912   313.3
  4956.8  313.26  4984.3  314.98  4992.3  310.79  4998.8   309.1  5003.8  309.08
  5006.5  308.58  5009.8  309.08  5013.2  314.04  5048.4  313.21  5085.2  317.31
  5112.4  322.11  5126.8  323.17  5186.9  331.79  5277.3   343.5  5290.9  344.01
#Mann= 5 ,-1 , 0
  4523.5     .16       0  4659.5     .12       0  5003.8     .07       0
  5009.8     .12       0  5186.9     .16       0
Bank Sta=4761.1,5085.2
XS Rating Curve= 0 ,0
Exp/Cntr=0.3,0.1

Type RM Length L Ch R = 1 ,1895    ,424,424,424
BEGIN DESCRIPTION:
BATSMITH CREEK 4.0
END DESCRIPTION:
XS GIS Cut Line= 3
      3646149.61     10613510.19      3646149.61     10613110.19
      3645999.61     10612710.19
#Sta/Elev= 30
  4609.3  342.03  4619.3  339.75  4659.3  333.52  4791.4  316.81  4799.3  315.54
  4849.3  310.01  4879.3  309.86  4979.3  312.15  4996.3  309.84  4999.1  309.34
  5002.3  309.84  5006.8  311.68  5024.4  312.34  5079.6  311.41    5085  312.16
  5140.1  310.69  5170.4  312.06  5195.3  315.09  5244.3  320.13  5255.8  322.61
  5265.6  322.91  5276.5  324.86    5287  327.71  5297.7  328.51  5351.1  337.45
  5366.2  338.78  5372.4  340.44  5383.1  341.02  5396.5  343.38  5436.5  346.41
#Mann= 5 ,-1 , 0
  4609.3     .16       0  4791.4     .12       0  4996.3     .07       0
  5002.3     .12       0  5276.5     .16       0
Bank Sta=4799.3,5195.3
XS Rating Curve= 0 ,0
Exp/Cntr=0.3,0.1

Type RM Length L Ch R = 1 ,1471    ,444,444,444
BEGIN DESCRIPTION:
BATSMITH CREEK 3.0
END DESCRIPTION:
XS GIS Cut Line= 3
      3646499.62     10613510.16      3646549.61     10613260.19
      3646249.62     10612460.21
#Sta/Elev= 30
  4734.2  340.28  4795.4  329.75  4877.7  318.48  4917.7  313.18  4958.5  309.28
  4991.8  310.66  4995.9  307.52  4998.7  307.02  5001.9  307.52  5010.5  310.31
  5138.6  308.78  5352.2  309.47  5406.5  308.04  5431.4  308.84  5480.4  312.98
  5485.6  313.31  5516.9  316.84    5530  320.08  5572.1  325.57  5587.2  328.71
  5602.3   329.6  5608.6  331.39  5651.3  336.56  5657.5  339.55  5687.8  344.59
  5702.1  348.56  5767.9  361.27  5779.4  361.88  5798.1  365.14  5843.5  367.65
#Mann= 7 ,-1 , 0
  4734.2     .16       0  4877.7     .12       0  4995.9     .07       0
  5001.9     .12       0  5485.6     .16       0    5530     .05       0
  5702.1     .16       0
Bank Sta=4917.7,5480.4
XS Rating Curve= 0 ,0
Exp/Cntr=0.3,0.1

Type RM Length L Ch R = 1 ,1027    ,547,547,547
BEGIN DESCRIPTION:
BATSMITH CREEK 2.0
END DESCRIPTION:
XS GIS Cut Line= 3
      3646849.61     10613410.19      3646799.61     10612960.19
      3646399.58     10612560.16
#Sta/Elev= 30
  4571.6  321.26  4583.4  319.72  4611.8  314.73    4642  311.55  4662.2   309.3
  4682.3  308.31  4722.5  309.24  4732.6  308.24  4752.7  308.87  4994.2  307.02
  5109.2  306.85  5137.5  307.44  5176.9  306.67  5179.7  306.17  5182.9  306.67
  5208.2  307.94  5250.6  308.56  5293.1   311.7  5377.9  315.94  5392.1  315.81
  5429.1  319.04  5448.6   320.6  5462.8  323.63  5476.9  325.32  5491.1  328.68
  5505.2  330.42  5519.3  333.81  5547.6  338.92  5586.5  345.13  5590.1  345.13
#Mann= 5 ,-1 , 0
  4571.6     .05       0  4583.4     .12       0  5176.9     .07       0
  5182.9     .12       0  5429.1     .05       0
Bank Sta=4642,5293.1
XS Rating Curve= 0 ,0
Exp/Cntr=0.3,0.1

Type RM Length L Ch R = 1 ,480     ,0,0,0
BEGIN DESCRIPTION:
BATSMITH CREEK 1.0
END DESCRIPTION:
XS GIS Cut Line= 4
      3646673.62     10613612.21      3647163.18      10613221.6
      3647163.18     10612580.98      3646465.23     10612060.12
#Sta/Elev= 30
  3912.1  343.71  4081.7  332.24  4116.9  328.09  4145.7  327.03    4181   322.4
  4249.3  316.73  4259.4  316.62  4294.6  312.26  4358.7  308.91    4522  306.55
  4599.8  307.26  5006.8  304.67  5009.6  304.17  5012.8  304.67  5048.7  308.09
  5069.8  309.84  5119.8  311.35  5268.4  309.92  5360.2  312.28  5424.8  315.51
  5489.4  320.48  5539.5  326.43  5554.1  329.31  5568.7  330.61  5645.8  344.66
  5689.6  349.35  5739.6  352.86  5789.6  354.02  5989.8   350.5  6049.9  351.07
#Mann= 5 ,-1 , 0
  3912.1     .05       0  4249.3     .12       0  5006.8     .07       0
  5012.8     .12       0  5048.7     .05       0
Bank Sta=4358.7,5069.8
XS Rating Curve= 0 ,0
Exp/Cntr=0.3,0.1

Chan Stop Cuts=-1
Use User Specified Reach Order=0
Composite Channel Slope=5
