HEC-RAS study LAKE CREEK.prj: LAKE CREEK Base Level Engineering

--- LAKE CREEK.g01 (geometry) --- (continued)

Type RM Length L Ch R = 1 ,111122  ,377,377,377
BEGIN DESCRIPTION:
LAKE CREEK 160.0
END DESCRIPTION:
XS GIS Cut Line= 3
      3721749.61     10665910.19      3720949.61     10665110.19
      3720199.64     10665160.19
#Sta/Elev= 30
  3860.7  364.44  3864.2  364.44  3874.8  359.97    3889  357.86  3973.8   355.1
  4002.1  351.96    4087  346.59  4101.1  344.49  4171.8  340.31  4242.5  336.96
  4369.8  335.57    4407  334.66  4437.9  334.62  4526.8  333.31  5184.1  332.74
  5209.6  332.46  5212.3  331.96  5215.6  332.46  5242.6  335.91  5272.7  336.82
  5302.8  335.41  5312.8  333.55  5342.8  332.66    5413  333.05  5463.1  334.97
  5513.2  338.36  5543.3  338.81  5601.7  343.41  5663.6  349.63  5743.7  355.66
#Mann= 8 ,-1 , 0
  3860.7     .05       0    4407     .12       0  4437.9     .05       0
  4526.8     .12       0  5184.1      .1       0  5209.6     .07       0
  5215.6      .1       0  5601.7     .05       0
#XS Ineff= 1 ,-1
 5263.21 5639.23  335.92
Permanent Ineff=
       F
Bank Sta=4369.8,5463.1
XS Rating Curve= 0 ,0
Exp/Cntr=0.3,0.1

Type RM Length L Ch R = 1 ,110745  ,500,500,500
BEGIN DESCRIPTION:
LAKE CREEK 159.0
END DESCRIPTION:
XS GIS Cut Line= 3
      3722342.02     10666308.29      3721245.36     10664845.67
      3720385.97     10664663.38
#Sta/Elev= 30
  3070.1     390  3219.9  386.38  3363.6  386.73  3555.3  380.84  3584.5  381.26
  3734.5  371.84  3949.1  352.97  3955.3  353.72  4099.1  342.22  4178.3  338.34
  4284.5  336.03  4378.3  335.95  4413.7  334.05  4534.5  333.69  4549.1  334.98
  4613.7  334.28  4619.9  332.53  4803.7  332.73  4975.6  330.13  5057.4  331.93
  5098.4  329.79  5156.6  329.66  5159.4  329.16  5162.6  329.66  5231.2  330.58
  5243.7  332.28  5364.1  335.07  5456.1  333.86  5602.2  336.28  5776.7  342.25
#Mann= 6 ,-1 , 0
  3070.1     .05       0  4803.7     .12       0  5156.6     .07       0
  5162.6     .12       0  5243.7      .1       0  5602.2     .05       0
Bank Sta=4413.7,5456.1
XS Rating Curve= 0 ,0
Exp/Cntr=0.3,0.1

Type RM Length L Ch R = 1 ,110245  ,511,511,511
BEGIN DESCRIPTION:
LAKE CREEK 158.0
END DESCRIPTION:
XS GIS Cut Line= 4
      3723235.41     10663470.94      3722421.57     10663747.58
      3721353.86     10664333.52      3720455.41     10664311.82
#Sta/Elev= 30
  2707.2  367.19  2839.7  371.02  3001.9  365.95  3122.1  370.47  3184.9  369.35
  3190.2  367.39  3310.4  370.14  3367.9  368.58  3430.6  362.38  3435.9  359.61
  3498.7  358.67  3556.2  361.55  3687.6  348.77  3953.9  334.95  4035.4  333.35
    4072  332.77  4128.3  330.79  4714.3  330.87    4969  332.18    4999  328.58
    5019  331.88    5026  327.99  5028.8  327.49    5032  327.99    5049     332
    5109  329.74  5159.1  333.06  5181.4  336.95  5349.1  345.27  5683.4  354.76
#Mann= 7 ,-1 , 0
  2707.2     .05       0  3953.9     .12       0    4072     .05       0
  4714.3     .12       0    5026     .07       0    5032     .12       0
  5181.4     .05       0
Bank Sta=4035.4,5159.1
XS Rating Curve= 0 ,0
Exp/Cntr=0.3,0.1

Type RM Length L Ch R = 1 ,109734  ,399,399,399
BEGIN DESCRIPTION:
LAKE CREEK 157.0
END DESCRIPTION:
XS GIS Cut Line= 3
      3722299.61     10663560.19      3721099.61     10663860.19
      3720699.65     10663960.18
#Sta/Elev= 30
  3738.1  364.52  3756.1  362.11  3761.3  364.31  3797.4   357.9  3802.5  359.38
  3838.6  352.24  3843.8  353.93  3851.5  350.89  3879.8  348.17    3885   348.9
  3954.6  341.83  4003.5  339.29  4498.3  332.11  4668.4  329.71  4869.4  328.78
  4977.6  330.41  4985.3  329.09  4990.1  326.84  4992.8  326.34  4996.1  326.84
    5006  326.87  5016.3  330.23  5026.6  330.95  5054.8  330.22    5109  329.17
  5148.1  332.49  5170.9  335.01  5315.2  345.17  5346.1  348.93  5387.3  350.82
#Mann= 5 ,-1 , 0
  3738.1     .05       0  4990.1     .03       0  4996.1     .05       0
  5054.8     .12       0  5148.1     .05       0
Bank Sta=4498.3,5148.1
XS Rating Curve= 0 ,0
Exp/Cntr=0.3,0.1

Type RM Length L Ch R = 1 ,109335  ,485,485,485
BEGIN DESCRIPTION:
LAKE CREEK 156.0
END DESCRIPTION:
XS GIS Cut Line= 3
      3721504.59     10663177.77        3720824.     10663615.29
      3720567.04     10663858.37
#Sta/Elev= 30
  4310.7  342.74  4316.6  342.74  4323.5   341.7  4329.4  342.58  4359.8  340.21
  4423.6  336.96  4447.4  336.47  4474.7  334.35  4685.1  331.07  4801.7  328.51
  4843.9  328.72  4922.9  327.85  4934.7  327.06  4937.5  326.56  4940.7  327.06
  4958.8  327.14    4974  328.93  4989.2  329.31  5004.4  328.12  5010.4  329.62
  5046.7  328.08    5083  331.02  5119.3  334.65  5168.6  338.34  5182.8  340.28
    5197  340.88  5232.6  344.56  5267.8  346.63  5338.6  348.94  5473.5  349.85
#Mann= 3 ,-1 , 0
  4310.7     .05       0  4934.7     .03       0  4940.7     .05       0
Bank Sta=4685.1,5083
XS Rating Curve= 0 ,0
Exp/Cntr=0.3,0.1

Type RM Length L Ch R = 1 ,108850  ,331,331,331
BEGIN DESCRIPTION:
LAKE CREEK 155.0
END DESCRIPTION:
XS GIS Cut Line= 3
      3720949.63     10662760.17      3720599.61     10663210.19
      3720549.61     10663710.18
#Sta/Elev= 30
  4411.1  361.93  4482.6  353.07  4503.4  351.82  4546.9  346.63  4567.7  346.17
    4603  342.86  4611.1   341.3  4631.9  340.46  4646.4  337.63  4667.2  337.18
  4710.7  332.51  4760.4  329.38  4895.3  325.29  4938.7  326.44    4945  324.63
  4953.2  326.91  4983.7  327.32  4991.3  327.04  4998.3  324.26  5001.1  323.76
  5004.3  324.26  5011.4  325.98  5021.4  326.82  5091.8  327.19  5111.9  328.08
  5121.9  329.86    5235   337.3  5282.7  337.86  5330.4  340.88  5483.7  344.01
#Mann= 3 ,-1 , 0
  4411.1     .05       0  4998.3     .03       0  5004.3     .05       0
Bank Sta=4760.4,5121.9
XS Rating Curve= 0 ,0
Exp/Cntr=0.3,0.1

Type RM Length L Ch R = 1 ,108519  ,534,534,534
BEGIN DESCRIPTION:
LAKE CREEK 154.0
END DESCRIPTION:
XS GIS Cut Line= 3
      3721011.51     10662594.45      3720587.89     10662816.68
      3719907.32     10663573.64
#Sta/Elev= 30
  4300.1  359.06  4348.9  357.51  4403.8  353.81  4409.4  354.48    4492  348.79
  4497.6  349.61  4607.9  344.27  4640.7  340.75  4662.8  339.41  4668.4  340.36
  4697.5   337.1  4712.6  337.01  4786.6  331.14  4857.7  328.04  4928.7  325.05
  4957.1  326.09    4975  322.05  4977.8  321.55    4981  322.05  4992.2  323.58
  5006.4  323.03  5013.1  326.18  5119.4  325.38    5212  327.94  5275.5  331.65
  5367.4  333.54  5466.8  338.01    5573  338.96  5622.3  337.14  5796.4  341.46
#Mann= 3 ,-1 , 0
  4300.1     .05       0    4975     .03       0    4981     .05       0
Bank Sta=4857.7,5212
XS Rating Curve= 0 ,0
Exp/Cntr=0.3,0.1

Type RM Length L Ch R = 1 ,107985  ,283,283,283
BEGIN DESCRIPTION:
LAKE CREEK 153.0
END DESCRIPTION:
XS GIS Cut Line= 2
       3721025.4     10662483.35      3719608.77     10662511.12
#Sta/Elev= 30
  4364.5  361.47  4450.3   355.8  4480.3  352.64  4650.3  338.73  4760.4  333.62
  4840.4  327.42  4870.4  326.07  4971.9  323.79  4990.4  323.03  4997.4  321.75
  5000.2  321.25  5003.4  321.75  5010.4  323.78  5020.4  324.48  5320.5  323.04
  5330.5  323.47  5350.5  326.25  5380.5  329.32  5420.5  331.18  5500.5  332.29
  5530.5  331.68  5540.5   332.6  5600.5  333.57  5610.5  332.54  5620.5  333.05
  5639.5   332.3  5700.5  333.27  5710.6     332  5730.6  332.39  5781.4  330.74
#Mann= 5 ,-1 , 0
  4364.5     .05       0  4997.4     .03       0  5003.4     .05       0
  5540.5     .12       0  5639.5     .16       0
Bank Sta=4870.4,5350.5
XS Rating Curve= 0 ,0
Exp/Cntr=0.3,0.1

Type RM Length L Ch R = 1 ,107702  ,1140,1140,1140
BEGIN DESCRIPTION:
LAKE CREEK 152.0
END DESCRIPTION:
XS GIS Cut Line= 3
      3721364.53     10662270.97      3720539.88     10662197.19
      3719606.67     10662323.06
#Sta/Elev= 30
  4010.9  355.03  4078.5   350.2  4176.5  347.87  4206.6  345.93  4276.9  347.71
    4307  346.51  4387.3  349.18  4618.2   334.5  4728.7  325.37  4778.9  322.68
  4889.6  324.36  4950.1  323.04  4980.4   323.9  4987.5  321.97  4990.2  321.47
  4993.5  321.97  5010.7   323.6  5040.9  322.88  5071.2  323.97    5384  322.25
  5414.3  325.21  5420.8  327.04  5425.9  326.46  5493.6  331.55  5627.2  332.23
    5644  332.26  5649.1  333.79  5666.5  332.39  5754.4  332.13  5780.5  332.75
#Mann= 5 ,-1 , 0
  4010.9     .05       0  4987.5     .03       0  4993.5     .05       0
  5627.2     .16       0  5754.4     .12       0
Bank Sta=4728.7,5414.3
XS Rating Curve= 0 ,0
Exp/Cntr=0.3,0.1

Type RM Length L Ch R = 1 ,106562  ,504,504,504
BEGIN DESCRIPTION:
LAKE CREEK 151.0
END DESCRIPTION:
XS GIS Cut Line= 3
      3722025.35     10661698.62      3720518.45      10661413.9
      3719633.69     10662183.36
#Sta/Elev= 30
  3632.9  388.92  3791.4  382.16  3801.6  375.47  3814.9  373.99  3832.1  377.23
  3943.7  361.11  4066.2   348.9  4076.3  346.89  4081.9  342.68  4134.2  342.24
  4153.6  339.08  4381.7  324.98  4516.1  322.73  4605.5  324.91  4673.2  320.16
  4994.7  319.66  4997.4  319.16  5000.7  319.66  5034.9  320.62  5176.6  321.25
  5181.5  321.16  5255.5  324.46  5483.1  326.91  5787.2  329.86  5952.9  328.53
  6025.8  329.82  6098.6   329.5  6240.1  336.94  6297.1  336.28    6339  335.11
#Mann= 12 ,-1 , 0
  3632.9     .05       0  3943.7     .16       0  4153.6     .05       0
  4994.7     .03       0  5000.7     .05       0  5034.9     .12       0
  5176.6     .16       0  5181.5     .12       0  5483.1     .16       0
  5952.9     .12       0  6025.8     .16       0  6297.1     .12       0
Bank Sta=4381.7,5255.5
XS Rating Curve= 0 ,0
Exp/Cntr=0.3,0.1

Type RM Length L Ch R = 1 ,106058  ,350,350,350
BEGIN DESCRIPTION:
Mapping XS f3deeeea
END DESCRIPTION:
XS GIS Cut Line= 3
      3722225.55     10660727.65      3720600.53     10661060.99
      3719615.38     10662114.75
#Sta/Elev= 30
  3613.8  348.02  3670.9  342.39  3783.2  336.09  3804.7  337.62  3834.2  334.22
  4089.4  331.16  4399.3   323.9  4477.9  322.01    4804  319.26  4926.5  320.99
    4996  318.67  4998.8  318.17    5002  318.67  5028.6  319.34  5079.6  324.92
  5120.5  324.76  5222.6  319.03  5456.7  322.92  5576.9  319.56  5612.5  320.31
  5644.4   323.9  5652.5  324.47  5966.2  329.02  6101.4  328.53  6206.6  326.42
  6297.1   327.4  6455.3  330.72  6560.2  330.46  6714.4  337.59  6715.2  337.59
#Mann= 10 ,-1 , 0
  3613.8     .05       0  4477.9     .12       0    4996     .07       0
    5002     .12       0  5644.4     .16       0  5652.5     .12       0
  6101.4     .16       0  6297.1     .12       0  6455.3     .16       0
  6714.4     .12       0
#XS Ineff= 1 ,-1
 5100.61 6505.59  324.85
Permanent Ineff=
       F
Bank Sta=4399.3,5644.4
XS Rating Curve= 0 ,0
Exp/Cntr=0.3,0.1

Type RM Length L Ch R = 1 ,105708  ,577,577,577
BEGIN DESCRIPTION:
LAKE CREEK 150.0
END DESCRIPTION:
XS GIS Cut Line= 4
      3721390.57     10659645.11       3720761.5     10660684.74
      3719880.05       10661414.       3719615.7     10662035.89
#Sta/Elev= 30
  3668.7  367.05  3747.9  369.13  4130.5  363.27  4182.8  360.26  4320.5  344.04
  4394.2  332.15  4415.5  331.67  4422.7  328.57  4473.7  325.71  4481.1  323.47
  4562.9  320.34  4697.7  317.89  4700.4  317.39  4703.7  317.89  4853.9  319.76
  5038.5  318.24  5094.5  324.04  5181.5  320.65  5215.7  319.61  5371.9  319.45
  5443.6  324.41  5556.9  324.04  5662.9   327.4  5936.6  328.04  6024.4   327.2
  6214.9  329.32  6351.8  330.42  6528.2  325.49  6577.6  326.16  6703.6  334.09
#Mann= 11 ,-1 , 0
  3668.7     .16       0  3747.9     .12       0  4697.7     .07       0
  4703.7     .12       0  5181.5     .16       0  5215.7     .12       0
  5662.9     .16       0  5936.6     .12       0  6024.4     .16       0
  6214.9     .12       0  6577.6     .16       0
#XS Ineff= 1 ,-1
 5097.05  5918.7  324.07
Permanent Ineff=
       F
Bank Sta=4473.7,5443.6
XS Rating Curve= 0 ,0
Exp/Cntr=0.3,0.1

Type RM Length L Ch R = 1 ,105131  ,616,616,616
BEGIN DESCRIPTION:
LAKE CREEK 149.0
END DESCRIPTION:
XS GIS Cut Line= 4
      3720483.72     10659886.14      3720178.17     10660733.35
      3719733.72     10661434.74      3719502.58     10662431.52
#Sta/Elev= 30
  4396.7   344.7  4691.1  331.23  4716.5  328.73  4869.9  323.09  4925.9  317.63
  5099.4  318.43  5166.1   316.7  5186.1  318.43  5252.8  318.63  5278.2  322.05
  5307.7  323.29  5395.8  325.76  5495.8  324.02  5656.8   326.1  5808.5  325.13
  5860.2  327.22  5996.6  327.21  6069.5  328.55  6075.4     330    6277  328.15
  6344.4  330.17  6492.6  327.15  6554.1  327.77  6562.9  326.42    6568  328.11
  6636.3  327.93  6786.4  337.27  6841.6  336.67  6924.7   331.9  7150.9  332.02
#Mann= 1 ,-1 , 0
  4396.7     .06       0
Bank Sta=4869.9,5307.7
XS Rating Curve= 0 ,0
Exp/Cntr=0.3,0.1

Type RM Length L Ch R = 1 ,104515  ,859,859,859
BEGIN DESCRIPTION:
LAKE CREEK 148.0
END DESCRIPTION:
XS GIS Cut Line= 3
      3719712.89     10660018.09      3719775.39     10660802.79
      3719449.26     10662425.56
#Sta/Elev= 30
  4518.5  360.54  4550.7  357.29    4661  339.98  4666.1  337.97  4681.1  337.43
  4711.2  332.62  4801.5  322.72  4871.5  314.75  4982.1  317.15  5142.6  316.59
  5222.8  322.32  5496.8  323.56  5614.1  322.33  5863.4  329.05  6016.1  329.19
  6088.4  326.69  6231.2  328.73  6435.2  327.32  6529.9   330.6  6575.7  334.25
  6580.8  331.95  6608.6  334.71  6631.7  333.21  6677.4  334.12  6682.5  332.34
  6751.4  329.33  6771.8  330.49  6779.2  332.66  6792.2  330.83  6960.9   331.6
#Mann= 1 ,-1 , 0
  4518.5     .06       0
Bank Sta=4801.5,5614.1
XS Rating Curve= 0 ,0
Exp/Cntr=0.3,0.1

Type RM Length L Ch R = 1 ,103656  ,452,452,452
BEGIN DESCRIPTION:
LAKE CREEK 147.0
END DESCRIPTION:
XS GIS Cut Line= 3
      3719317.07     10659802.75      3719087.89     10660469.46
      3718611.75     10662776.34
#Sta/Elev= 30
    4146  342.53  4333.2  336.71  4588.5  324.93  4765.3  322.22  4984.2  314.09
  5068.2  317.76  5188.7  315.19    5444  315.89  5515.4  321.55  5576.7  319.53
  5648.2  322.47  5957.6  329.68  6304.3  344.81  6500.3  348.52  6550.5  348.94
  6595.7  344.11  6600.8  346.47  6638.6  342.18  6746.5   337.8  6751.6  341.84
  6771.4   343.3  6796.7  339.42  6822.4  339.31  6863.3  339.57  6883.7   342.2
  6942.4  340.92  6997.8  342.77  7042.9  339.69  7138.4   339.5  7206.5  342.64
#Mann= 1 ,-1 , 0
    4146     .06       0
Bank Sta=4765.3,5648.2
XS Rating Curve= 0 ,0
Exp/Cntr=0.3,0.1

Type RM Length L Ch R = 1 ,103204  ,297,297,297
BEGIN DESCRIPTION:
LAKE CREEK 146.0
END DESCRIPTION:
XS GIS Cut Line= 3
      3718492.88     10659416.09      3718712.89     10660587.51
      3718448.99       10661782.
#Sta/Elev= 30
  3690.7  345.51  3857.6  355.24    3878  357.75  3972.8  358.62  4071.3   347.9
  4091.7   343.6  4122.2  341.27  4152.7  333.82    4224  323.16  4274.8  316.28
  4833.6  315.37  4875.2  317.21  4881.4  314.12  5013.5  314.42  5018.4  312.92
  5131.1  316.43  5192.6  314.24  5290.9  314.51  5339.6  317.45  5407.6  315.15
  5568.2  315.08  5573.3  316.85  5581.7  315.31    5633  314.98  5745.6  317.31
  5776.3   321.5  5878.7  332.11  5894.3  335.88  5981.2  345.29  6105.9  348.24
#Mann= 1 ,-1 , 0
  3690.7     .06       0
Bank Sta=4224,5776.3
XS Rating Curve= 0 ,0
Exp/Cntr=0.3,0.1

Type RM Length L Ch R = 1 ,102907  ,501,501,501
BEGIN DESCRIPTION:
LAKE CREEK 145.0
END DESCRIPTION:
XS GIS Cut Line= 4
      3718232.46     10660097.49      3718299.61     10660510.19
      3718449.61     10660810.19      3717999.63     10661410.16
#Sta/Elev= 30
  4227.5  335.43  4250.5  333.35    4291  333.02  4311.3  331.44  4341.7  332.81
  4366.2  332.04  4473.4  335.54  4489.3  337.64  4503.8  336.88  4544.3  339.73
  4612.3  341.43  4617.4  342.96    4654  341.97  4659.6  342.97  4712.7  335.37
  4721.1  335.25  4726.7  333.22  4802.2  324.89  4816.1  321.67  4877.6  313.81
  4958.7  314.43  4991.6  313.37  4994.3  312.87  4997.6  313.37  5088.3  315.93
    5131  314.38  5387.3  314.27  5538.3  321.72    5631  327.22    5731  338.44
#Mann= 3 ,-1 , 0
  4227.5     .12       0  4991.6     .07       0  4997.6     .12       0
Bank Sta=4816.1,5538.3
XS Rating Curve= 0 ,0
Exp/Cntr=0.3,0.1

Type RM Length L Ch R = 1 ,102406  ,439,439,439
BEGIN DESCRIPTION:
LAKE CREEK 144.0
END DESCRIPTION:
XS GIS Cut Line= 3
       3718199.6      10660560.2      3717999.61     10660810.19
       3717699.6     10661010.19
#Sta/Elev= 30
  4686.9  337.78  4722.9   334.5  4786.9  325.08  4814.9  322.13  4828.6  318.99
  4836.6  315.56    4851  314.09    4879   313.8  4883.2  312.93  4885.9  312.43
  4889.2  312.93  4892.6  313.73  4929.4   313.9    4943  313.23  4964.6  313.78
    4971  312.97  5050.6  313.61  5107.7  317.06  5151.3  321.68  5179.8  323.31
  5200.8  325.92  5215.9  326.42  5223.4  328.72  5236.9  329.25  5266.9  333.73
    5288   335.3    5309  338.95    5324  339.89  5331.5  342.06  5367.6  345.82
#Mann= 3 ,-1 , 0
  4686.9     .12       0  4883.2     .07       0  4889.2     .12       0
Bank Sta=4814.9,5151.3
XS Rating Curve= 0 ,0
Exp/Cntr=0.3,0.1

Type RM Length L Ch R = 1 ,101967  ,531,531,531
BEGIN DESCRIPTION:
LAKE CREEK 143.0
END DESCRIPTION:
XS GIS Cut Line= 3
      3718199.57      10660360.2      3717799.61     10660460.19
      3717599.59      10660560.2
#Sta/Elev= 30
  4602.6   343.9  4633.5  341.19  4661.8  336.72  4695.3  333.66  4703.1  331.75
  4708.2  331.86  4715.9  330.05  4736.6  328.85  4744.3  327.46  4757.2  326.94
  4785.5  324.14    4819   322.5  4826.8  320.61  4860.3  317.79    4868   316.3
  4880.9  316.01  4922.1   312.7    4984  313.16  4988.7  312.46  4991.4  311.96
  4994.7  312.46  5045.6  312.56    5068  315.02  5073.6  314.93  5095.9  318.23
  5126.7  320.95  5157.4   325.6    5163  325.53  5216.1  331.14  5238.5  332.55
#Mann= 3 ,-1 , 0
  4602.6     .12       0  4988.7     .07       0  4994.7     .12       0
Bank Sta=4826.8,5126.7
XS Rating Curve= 0 ,0
Exp/Cntr=0.3,0.1

Type RM Length L Ch R = 1 ,101436  ,401,401,401
BEGIN DESCRIPTION:
LAKE CREEK 142.0
END DESCRIPTION:
XS GIS Cut Line= 3
      3718371.37     10659732.92      3717714.28      10660053.9
       3717449.6      10660460.2
#Sta/Elev= 30
  4268.7  348.53    4275  349.58  4281.8  347.31  4333.1  345.32  4438.3  343.22
  4528.3  344.48  4567.8  342.36  4640.9  342.25  4693.6  336.63  4725.5  331.27
    4731  332.85  4738.1  329.91  4776.1  326.25  4804.9  321.05  4821.1  320.25
  4830.2  317.71  4837.7  316.71  4866.2  312.43  4882.8  312.38  4888.7  313.97
  4996.8  312.29  4999.6  311.79  5002.8  312.29  5066.9  315.88    5103  319.53
  5166.4  324.89    5282  331.39  5353.6  333.56  5462.2  332.79  5484.9  334.38
#Mann= 6 ,-1 , 0
  4268.7     .16       0  4333.1     .12       0  4830.2     .16       0
  4837.7     .12       0  4996.8     .07       0  5002.8     .12       0
Bank Sta=4821.1,5103
XS Rating Curve= 0 ,0
Exp/Cntr=0.3,0.1

Type RM Length L Ch R = 1 ,101035  ,461,461,461
BEGIN DESCRIPTION:
LAKE CREEK 141.0
END DESCRIPTION:
XS GIS Cut Line= 2
      3717810.11     10658997.25      3717226.79     10660559.72
#Sta/Elev= 30
  4195.2  348.29  4201.1  348.16  4283.7  344.72  4378.5  335.77  4422.5  329.21
  4486.5  324.48  4726.1  323.54  4751.1  320.89  4774.7  321.61  4781.4  319.49
  4796.1  318.92  4849.5  312.64  4910.5  312.18  4913.3  311.68  4916.5  312.18
  5030.9  312.47  5098.8  318.64  5169.7  326.27    5245  328.66  5294.9  327.58
  5300.3  325.49  5319.1  326.81  5385.8  323.06  5410.8  323.82  5416.1  321.88
    5557  320.65  5628.7  322.87  5753.1  335.56  5831.5  340.88    5863  340.84
#Mann= 4 ,-1 , 0
  4195.2      .1       0  4201.1     .12       0  4910.5     .07       0
  4916.5     .12       0
#XS Ineff= 1 ,-1
 5241.87 5857.72  328.76
Permanent Ineff=
       F
Bank Sta=4796.1,5098.8
XS Rating Curve= 0 ,0
Exp/Cntr=0.3,0.1

Type RM Length L Ch R = 1 ,100574  ,368,368,368
BEGIN DESCRIPTION:
LAKE CREEK 140.0
END DESCRIPTION:
XS GIS Cut Line= 3
       3717462.9     10658761.11      3717087.89     10659552.79
      3717108.68     10660627.18
#Sta/Elev= 30
  3933.8  344.53  3970.9  342.17  4093.3  335.94  4098.8   334.4    4116  335.09
  4235.3  326.79  4252.5   327.7    4258  325.55  4326.3  324.11  4408.6  319.04
  4559.2  321.58  4678.5  318.62  4695.7  316.33  4701.2  318.09    4726  313.04
  4789.2  311.87    4792  311.37  4795.2  311.87  4805.4  312.23  5116.6  312.26
  5177.3  314.37  5258.4  312.61  5387.3  313.64  5467.3  318.03  5627.4  328.19
  5667.4   329.1  5673.1   327.1  5687.4  330.03  5737.4  334.41  5884.4  343.08
#Mann= 8 ,-1 , 0
  3933.8     .05       0  3970.9     .12       0    4726     .16       0
  4789.2     .07       0  4795.2     .16       0  4805.4     .12       0
  5116.6     .16       0  5258.4     .12       0
#XS Ineff= 1 ,-1
 5250.51 5789.13  326.94
Permanent Ineff=
       F
Bank Sta=4678.5,5467.3
XS Rating Curve= 0 ,0
Exp/Cntr=0.3,0.1

Type RM Length L Ch R = 1 ,100206  ,904,904,904
BEGIN DESCRIPTION:
LAKE CREEK 139.0
END DESCRIPTION:
XS GIS Cut Line= 3
      3717018.45     10658587.51      3716733.72     10659629.18
      3716921.22     10660601.39
#Sta/Elev= 30
  3795.3  328.09  3815.9  325.63  3890.2  320.65  4026.1  317.91    4188  319.86
  4193.2  321.66  4341.6  321.37  4461.6  318.58  4603.9  320.68    4723  317.68
  4736.2  317.24  4877.5  315.32  4925.1  312.26  4944.5  311.81  4947.2  311.31
  4950.5  311.81  5021.6  311.94  5173.3  312.41  5344.7  312.53  5404.3  319.04
  5461.3   320.4  5466.9  322.02  5507.6  319.38    5528  323.77    5547   325.3
    5622  329.91  5690.9  338.62  5731.4  340.22  5805.6  341.28  5865.3  341.96
#Mann= 12 ,-1 , 0
  3795.3     .05       0  3815.9     .16       0  3890.2     .12       0
  4736.2     .16       0  4925.1     .12       0  4944.5     .07       0
  4950.5     .12       0  5021.6     .16       0  5173.3     .12       0
    5547     .05       0  5731.4     .12       0  5805.6     .05       0
#XS Ineff= 1 ,-1
 5349.59 5761.18  324.83
Permanent Ineff=
       F
Bank Sta=4723,5404.3
XS Rating Curve= 0 ,0
Exp/Cntr=0.3,0.1

Type RM Length L Ch R = 1 ,99302   ,259,259,259
BEGIN DESCRIPTION:
LAKE CREEK 138.0
END DESCRIPTION:
XS GIS Cut Line= 3
      3716960.28     10658572.64      3716173.81     10659458.08
      3715533.43     10659829.93
#Sta/Elev= 30
  3707.8  329.61  3805.8  321.33  3950.8  318.62  4025.5  318.09  4089.3  320.74
  4117.7  317.71  4330.1  318.26  4336.8  315.15  4344.3  316.92    4351  314.59
  4379.4  313.47  4407.9  314.33  4414.6  316.61  4422.1  313.93  4428.8  317.89
  4477.7   318.5  4527.7  319.08  4582.3  320.32  4634.5  318.28  4719.8  311.35
  4839.2  311.25  4858.1  310.89  4860.9  310.39  4864.1  310.89  5037.5   311.5
  5116.7  311.43  5241.4  317.07  5423.6  329.91  5601.7   335.3  5632.6  337.95
#Mann= 10 ,-1 , 0
  3707.8     .16       0  3950.8     .05       0  4477.7     .16       0
  4527.7     .05       0  4582.3     .12       0  4839.2     .07       0
  4858.1     .07       0  4864.1     .07       0  5037.5     .16       0
  5601.7     .05       0
#XS Ineff= 1 ,-1
 3769.31  4574.7  319.15
Permanent Ineff=
       F
Bank Sta=4330.1,5241.4
XS Rating Curve= 0 ,0
Exp/Cntr=0.3,0.1

Type RM Length L Ch R = 1 ,99043   ,71,71,71
BEGIN DESCRIPTION:
Mapping XS fafe9112
END DESCRIPTION:
XS GIS Cut Line= 4
       3716849.1     10658486.46       3716313.1     10659089.73
      3715881.24     10659365.34      3715517.73      10659666.1
#Sta/Elev= 30
  3727.8  337.86  3900.1  325.47  4062.7  319.58  4155.1  318.64  4218.7  320.86
  4226.2  318.32  4254.5  317.25  4332.4   316.4  4416.9  322.69  4459.5  322.81
  4539.8  320.42  4635.6  311.03    4646  310.92  4844.4  310.24  4899.4  310.04
  4929.9  313.09  4935.8  309.49  5023.8  309.27  5037.2  309.83  5050.5  313.41
  5065.6  313.07  5084.8  308.46  5087.5  307.96  5090.8  308.46    5123  312.77
  5143.8  318.39  5201.1  325.68  5264.9  327.63  5406.9  340.05  5518.9  340.09
#Mann= 8 ,-1 , 0
  3727.8     .16       0  4062.7     .05       0  4635.6     .12       0
    4646     .07       0  4844.4     .12       0  5050.5     .05       0
  5084.8     .07       0  5090.8     .05       0
#XS Ineff= 1 ,-1
 3931.91 4470.53   319.2
Permanent Ineff=
       F
Bank Sta=4254.5,5143.8
XS Rating Curve= 0 ,0
Exp/Cntr=0.3,0.1

Type RM Length L Ch R = 1 ,98972   ,47,47,47
BEGIN DESCRIPTION:
Mapping XS 771dc158
END DESCRIPTION:
XS GIS Cut Line= 5
      3716796.23     10658478.88      3716374.33     10658986.72
      3716020.16     10659213.28      3715934.22     10659270.58
      3715486.28     10659624.76
#Sta/Elev= 30
  3709.4  337.53  3835.9  328.73  4056.1  320.93  4197.8  321.37  4290.3  317.42
  4375.4  324.76  4541.4  326.72  4565.1  326.51  4575.6  320.61  4636.4   316.5
  4680.1  315.82  4731.4  327.13  4897.1  326.78  4911.3   325.5  4917.6  321.23
  4932.1  325.85  4938.4  313.08  4946.5  316.83  4952.9  309.53  4992.2  310.29
  4999.6  308.25  5002.3  307.75  5005.6  308.25  5045.9   308.6  5116.4  316.21
  5124.4  321.02  5153.3  326.32  5252.6  330.54  5337.6  339.03  5464.4  341.39
#Mann= 6 ,-1 , 0
  3709.4     .16       0  4056.1     .05       0  4575.6     .12       0
  4992.2     .05       0  4999.6     .03       0  5005.6     .05       0
#XS Ineff= 1 ,-1
 4054.88 4841.46  317.66
Permanent Ineff=
       F
Bank Sta=4636.4,5116.4
XS Rating Curve= 0 ,0
Exp/Cntr=0.3,0.1

Type RM Length L Ch R = 1 ,98925   ,236,236,236
BEGIN DESCRIPTION:
Mapping XS 1d094670
END DESCRIPTION:
XS GIS Cut Line= 3
      3716736.27     10658462.57      3716239.32      10659026.8
       3715463.5     10659538.23
#Sta/Elev= 30
  3741.7   338.9  3865.2  330.46  3928.8   331.7  3978.4  326.44  4092.2  323.77
  4198.2  325.07  4269.3  319.02    4276  314.39  4325.3  314.75  4389.8  324.51
  4558.8  311.56  4603.3   313.6  4705.8  310.71  4711.7  313.12  4726.8  310.37
  4828.6  314.47  4856.3  311.41  4877.3  315.19  4979.6  318.06  4985.8  313.91
  5018.9  308.35  5021.6  307.85  5024.9  308.35  5088.2  316.42  5109.2  318.91
  5124.3  326.37  5160.4  329.93  5253.8  333.16    5326   340.4  5422.8  341.17
#Mann= 6 ,-1 , 0
  3741.7     .16       0  4092.2     .05       0  4558.8     .12       0
  4979.6     .05       0  5018.9     .03       0  5024.9     .05       0
#XS Ineff= 1 ,-1
 4163.01 4410.98  318.67
Permanent Ineff=
       F
Bank Sta=4269.3,5088.2
XS Rating Curve= 0 ,0
Exp/Cntr=0.3,0.1

Type RM Length L Ch R = 1 ,98689   ,345,345,345
BEGIN DESCRIPTION:
LAKE CREEK 137.0
END DESCRIPTION:
XS GIS Cut Line= 3
      3716364.53     10658626.44       3715793.6     10659051.83
      3715424.23     10659291.14
#Sta/Elev= 30
  4217.5  338.74  4289.3  338.62    4378  329.13    4402   325.5  4437.4  322.77
    4452  324.37  4460.4  322.39  4466.6  322.81  4473.1  321.99  4481.2  318.25
  4487.5  317.08  4505.1  314.19  4522.9  314.62  4610.2  310.43  4616.8  312.13
  4631.4  312.65  4937.9  311.96  4953.1  308.97  5004.5  308.57  5014.6  307.09
  5017.4  306.59  5020.6  307.09  5022.6  307.46  5031.6  308.13  5040.8  316.14
  5046.7  314.68  5053.4   316.3  5061.9  318.13    5113   319.3  5369.6  335.89
#Mann= 7 ,-1 , 0
  4217.5     .16       0  4289.3     .05       0    4378     .07       0
  4505.1     .12       0  5014.6     .07       0  5020.6     .12       0
  5022.6     .05       0
Bank Sta=4487.5,5053.4
XS Rating Curve= 0 ,0
Exp/Cntr=0.3,0.1

Type RM Length L Ch R = 1 ,98344   ,499,499,499
BEGIN DESCRIPTION:
LAKE CREEK 136.0
END DESCRIPTION:
XS GIS Cut Line= 3
      3716399.64     10658260.16      3715699.61     10658760.19
       3715199.6     10658910.19
#Sta/Elev= 30
  4148.9  356.29  4241.1  349.01    4283  343.78  4292.7  344.22  4313.6  340.25
  4378.7  334.18    4407  329.79  4435.3  327.94  4443.9  325.75  4556.9  316.12
  4687.2  309.99    4788  311.12  4808.9  309.56  4923.2  310.92    4960  309.42
  4987.1  310.65  4995.7  309.09  5001.8  310.49  5003.1  306.17  5005.9  305.67
  5009.1  306.17  5011.8  306.17  5025.7  312.11  5050.9  312.45    5064  315.71
  5130.1  313.23    5154  313.79  5267.6  315.54  5353.7   319.3  5531.2  336.79
#Mann= 5 ,-1 , 0
  4148.9     .05       0    4283     .12       0  5003.1     .07       0
  5009.1     .12       0    5154     .05       0
Bank Sta=4556.9,5267.6
XS Rating Curve= 0 ,0
Exp/Cntr=0.3,0.1

Type RM Length L Ch R = 1 ,97845   ,554,554,554
BEGIN DESCRIPTION:
LAKE CREEK 135.0
END DESCRIPTION:
XS GIS Cut Line= 3
      3716399.61     10658210.19      3715649.61     10658310.19
       3715049.6     10658510.19
#Sta/Elev= 30
  4250.4  358.16    4292  354.83  4325.9  350.68  4351.3  349.08  4391.6  343.54
  4472.3  335.86  4527.4  331.57  4553.1   327.9  4592.7  324.28  4684.2   316.3
  4734.6  312.19    4775  310.39  4785.1  311.23  4805.3  309.05  4898.1  309.44
  4965.4  308.32  4986.9   310.5  4996.9  308.11  5001.5  305.22  5004.3  304.72
  5007.5  305.22  5038.7  309.41  5207.3  311.22  5302.2  315.27  5344.3  317.56
  5365.4  320.65    5376   319.9  5470.8  326.24  5544.6  329.26  5639.5  336.64
#Mann= 7 ,-1 , 0
  4250.4     .05       0  4325.9     .12       0  4527.4     .16       0
  4592.7     .12       0  4898.1     .05       0  5001.5     .03       0
  5007.5     .05       0
Bank Sta=4684.2,5302.2
XS Rating Curve= 0 ,0
Exp/Cntr=0.3,0.1

Type RM Length L Ch R = 1 ,97291   ,528,528,528
BEGIN DESCRIPTION:
LAKE CREEK 134.0
END DESCRIPTION:
XS GIS Cut Line= 3
      3715899.59      10657610.2      3715499.61     10657810.19
      3714949.65     10658060.17
#Sta/Elev= 30
    4576   348.8  4643.1  342.47  4687.8   335.9  4718.5   329.4  4724.1  329.61
  4799.6  319.62  4813.6  319.92  4830.3   316.9  4844.3   315.2  4866.7  312.91
  4933.8  309.08  4978.5  309.19  4986.9  308.52  4989.4  303.96  4992.2  303.46
  4995.4  303.96  5000.8  304.07  5020.4  308.45  5082.7  308.52  5156.3   308.7
    5166  308.58  5175.9  311.09  5220.9  315.13  5348.3  323.17  5440.6  323.94
  5492.2  326.66  5515.3  326.82  5579.1  331.48  5613.1  333.85  5627.3   333.8
#Mann= 7 ,-1 , 0
    4576     .05       0  4830.3     .12       0  4989.4     .07       0
  4995.4     .12       0  5082.7     .16       0  5156.3     .05       0
  5579.1     .12       0
Bank Sta=4844.3,5220.9
XS Rating Curve= 0 ,0
Exp/Cntr=0.3,0.1

Type RM Length L Ch R = 1 ,96763   ,434,434,434
BEGIN DESCRIPTION:
LAKE CREEK 133.0
END DESCRIPTION:
XS GIS Cut Line= 4
      3715857.43     10657306.14      3715162.97     10657392.95
      3714949.61     10658010.19      3714812.29     10658955.32
#Sta/Elev= 30
  4406.6  336.09  4456.2  333.08  4479.8  333.61  4555.4  327.68    4641  327.01
  4668.3  324.43  4721.6  321.38  4747.1  316.53  4777.3  314.57  4802.3  311.34
    4999  307.75  5006.1  305.28  5008.8  304.78  5012.1  305.28  5039.1  308.68
  5091.6  308.52  5136.3  312.27  5198.8  313.96  5320.7  317.58    5531  321.86
  5769.6  333.31  5891.4  334.71    5992  334.95  6153.6  329.33  6224.4  328.78
  6264.8  330.39  6295.1     329  6420.9  329.81  6467.2  331.78  6714.6  339.81
#Mann= 9 ,-1 , 0
  4406.6     .12       0  4456.2     .05       0  4668.3     .12       0
  5006.1     .07       0  5012.1     .12       0  5091.6     .05       0
  5320.7     .12       0  5891.4     .16       0  6467.2     .05       0
Bank Sta=4777.3,5198.8
XS Rating Curve= 0 ,0
Exp/Cntr=0.3,0.1

Type RM Length L Ch R = 1 ,96329   ,112,112,112
BEGIN DESCRIPTION:
Mapping XS 63a76d9d
END DESCRIPTION:
XS GIS Cut Line= 3
      3715879.87     10656910.43      3715055.19     10657018.94
      3713715.02     10657201.98
#Sta/Elev= 30
  4361.1  336.83  4470.8  337.02  4549.4  334.98  4694.2  336.01  4774.9   328.7
  4785.4  325.37    4854  317.42  4895.8  315.22  4926.2   312.9  4966.5  309.71
  4986.7  304.86  5008.4  304.31  5011.1  303.81  5014.4  304.31  5027.1  308.68
  5091.9  310.01  5117.8  310.77  5158.2  308.58  5168.7  310.21  5178.3  309.07
  5259.1  311.17  5308.7  309.77    5471  312.66  5662.8  313.93  5733.4  318.63
  5955.5  325.92  6106.9  327.47  6308.7  332.13  6423.1  330.97  6545.5  325.94
#Mann= 5 ,-1 , 0
  4361.1     .05       0  4895.8     .12       0  5008.4     .07       0
  5014.4     .12       0  5091.9     .05       0
Bank Sta=4926.2,5471
XS Rating Curve= 0 ,0
Exp/Cntr=0.3,0.1

Type RM Length L Ch R = 1 ,96217   ,140,140,140
BEGIN DESCRIPTION:
LAKE CREEK 132.0
END DESCRIPTION:
XS GIS Cut Line= 3
      3715806.03     10656775.89      3714990.09     10656927.79
      3714353.36     10656923.46
#Sta/Elev= 30
  4402.7  328.28  4559.8  324.56  4564.8  325.79  4612.5  325.29  4728.2  331.32
  4765.2  327.53  4775.4  328.65    4786  318.79  4797.7  318.37  4820.3  317.38
  4856.8  315.31  4958.5  313.68  4968.7  311.91  4978.9  304.92    4994  301.48
  4996.7  300.98    5000  301.48  5019.5  302.85  5029.7  305.91  5049.7  308.36
  5101.8  310.51  5203.2  310.61  5343.1  311.76  5401.8  310.24  5403.8  310.29
  5553.1   312.6  5623.1  315.61  5793.2  326.82  5823.2  330.03  5869.4  331.47
#Mann= 9 ,-1 , 0
  4402.7     .05       0  4797.7     .07       0  4820.3     .05       0
    4994     .04       0    5000     .05       0  5101.8     .16       0
  5203.2     .05       0  5401.8     .16       0  5403.8     .05       0
Bank Sta=4958.5,5553.1
XS Rating Curve= 0 ,0
Exp/Cntr=0.3,0.1

Type RM Length L Ch R = 1 ,96077   ,572,572,572
BEGIN DESCRIPTION:
Mapping XS 78834839
END DESCRIPTION:
XS GIS Cut Line= 3
      3715832.13     10656697.76      3714890.26     10656771.54
       3714195.8      10656745.5
#Sta/Elev= 30
    4380  321.78  4471.5  319.19  4482.8  320.19    4543  317.16  4605.7  319.19
  4791.2  319.31  4813.8  319.36  4890.7  315.09  4934.2  312.69  4988.3  307.59
  5001.4  300.72  5004.2  300.22  5007.4  300.72  5024.5  309.46  5034.5  310.47
  5084.7  308.24  5124.8   309.6  5189.3  308.68  5288.9  308.78  5335.4  308.35
    5388  309.74  5439.9  311.05  5465.5   312.3  5585.6  318.35  5685.7  324.69
  5705.7  327.07  5835.8  333.03  5905.8  337.44  5975.9  344.21  6019.7  345.58
#Mann= 9 ,-1 , 0
    4380     .05       0  4791.2     .07       0  4890.7     .12       0
  5001.4     .07       0  5007.4     .12       0  5189.3     .16       0
  5288.9     .12       0    5388     .16       0  5439.9     .05       0
Bank Sta=4934.2,5465.5
XS Rating Curve= 0 ,0
Exp/Cntr=0.3,0.1

Type RM Length L Ch R = 1 ,95505   ,484,484,484
BEGIN DESCRIPTION:
LAKE CREEK 131.0
END DESCRIPTION:
XS GIS Cut Line= 4
      3716352.96     10656519.81      3715992.69     10656437.34
      3715324.29     10656337.51      3714226.23     10656320.15
#Sta/Elev= 30
  3830.9  323.93  3936.5  322.81  3998.5   319.1  4244.1  310.93    4296  309.42
  4364.8   308.3  4749.6   306.4  4794.2  307.59  4804.4  307.62    4891  308.06
    4901  306.41    4941  305.33    4961  308.58    4971  308.43    4981  302.58
    5008  300.28  5010.8  299.78    5014  300.28  5019.7  303.57  5024.7  300.61
    5041   308.5    5071  306.81    5171  306.89    5241   307.9    5271  311.77
    5311  316.07    5358  318.35  5601.1  322.44  5821.1  329.68  5974.5  336.54
#Mann= 8 ,-1 , 0
  3830.9     .05       0    4296     .07       0  4364.8     .12       0
  4794.2     .05       0  4804.4     .12       0    5008     .07       0
    5014     .12       0    5358     .05       0
#XS Ineff= 2 , 0
         4480.69  321.01
Permanent Ineff=
       F       F
Bank Sta=4244.1,5271
XS Rating Curve= 0 ,0
Exp/Cntr=0.3,0.1

Type RM Length L Ch R = 1 ,95021   ,509,509,509
BEGIN DESCRIPTION:
LAKE CREEK 130.0
END DESCRIPTION:
XS GIS Cut Line= 3
      3717318.02     10655707.14      3716448.42     10655938.21
      3714430.15      10655873.1
#Sta/Elev= 30
  2920.7  330.82  2993.8  328.06  3206.4  326.62  3420.1  322.62  3455.1  323.97
  3620.1  318.23  3732.9  316.43  3826.7  314.89  3925.6  314.69  4109.5  311.51
  4149.5  310.74  4218.6  309.94  4494.1  306.64  4639.7  304.88  4979.9  307.04
  4989.9  306.81  4999.9  300.22  5006.9   299.9  5009.7   299.4  5012.9   299.9
  5019.9  307.24  5029.9  307.68  5079.9  305.06  5290.1  310.64  5420.1  319.95
  5465.8  318.65  5530.2  315.64  5540.2  318.65  5560.2  319.48  5839.8  325.65
#Mann= 12 ,-1 , 0
  2920.7     .05       0  3206.4     .16       0  3620.1     .05       0
  3732.9     .12       0  3826.7     .16       0  3925.6     .05       0
  4109.5     .16       0  4218.6     .05       0  4494.1     .12       0
  5006.9     .07       0  5012.9     .12       0  5465.8     .05       0
#XS Ineff= 2 , 0
         4129.06  317.98
Permanent Ineff=
       F       F
Bank Sta=4149.5,5290.1
XS Rating Curve= 0 ,0
Exp/Cntr=0.3,0.1

Type RM Length L Ch R = 1 ,94512   ,525,525,525
BEGIN DESCRIPTION:
LAKE CREEK 129.0
END DESCRIPTION:
XS GIS Cut Line= 3
      3715999.57      10655060.2      3715199.61     10655410.19
      3714549.63     10655310.19
#Sta/Elev= 30
    4118  343.83  4139.8  340.82    4369  323.65  4434.9  316.79  4528.4  310.96
  4552.5  308.49  4618.6  304.79  4663.7  304.71  4685.5  302.95  4703.1  304.83
  4784.2  304.64  4794.7  306.18  4807.6  303.97  4816.5  305.35  4871.1  304.54
  4982.2   306.3  4988.4  300.25  4998.3  299.74    5001  299.24  5004.3  299.74
  5011.4  303.66  5025.3  306.58  5122.7  304.99  5264.3  310.53  5409.9  319.07
  5476.8  325.74  5551.4  330.22  5598.2  335.12  5619.7  338.89  5648.8  340.87
#Mann= 6 ,-1 , 0
    4118     .12       0  4552.5     .16       0  4618.6     .12       0
  4998.3     .07       0  5004.3     .12       0  5409.9     .16       0
Bank Sta=4528.4,5264.3
XS Rating Curve= 0 ,0
Exp/Cntr=0.3,0.1

Type RM Length L Ch R = 1 ,93987   ,584,584,584
BEGIN DESCRIPTION:
LAKE CREEK 128.0
END DESCRIPTION:
XS GIS Cut Line= 3
      3715849.58     10655010.19      3715049.61     10654910.19
      3714549.63     10655260.17
#Sta/Elev= 30
  4229.6  334.44    4348  324.45  4390.8  319.32  4400.9  319.39  4421.1  315.62
  4501.7  309.38  4589.9  304.68  4662.9  302.42  4773.8  302.81  4844.3  304.49
  4874.6  304.37  4894.7  302.73  4945.1  305.69  4965.3  304.31  4985.4  305.21
    4995  299.81  4997.8  299.31    5001  299.81  5005.6   303.8  5015.6  305.49
  5072.4  309.27  5129.5  314.76  5182.4  316.25  5308.3   319.2  5358.8  318.55
  5451.3  322.33  5524.1  328.06  5560.7  332.32    5603  334.19  5646.1  340.39
#Mann= 4 ,-1 , 0
  4229.6     .12       0    4995     .07       0    5001     .12       0
  5182.4     .16       0
Bank Sta=4501.7,5072.4
XS Rating Curve= 0 ,0
Exp/Cntr=0.3,0.1

Type RM Length L Ch R = 1 ,93403   ,793,793,793
BEGIN DESCRIPTION:
LAKE CREEK 127.0
END DESCRIPTION:
XS GIS Cut Line= 2
      3715964.39     10654623.63      3714130.58     10654591.07
#Sta/Elev= 30
  4371.3  327.06  4455.9  320.24  4506.1  318.76  4656.1  309.08  4750.7   304.5
  4866.2  301.51  4876.2  302.49  4896.2   300.5  4906.2  302.19  4966.2   303.5
  4986.2  298.63  4996.2  299.74  5006.2   304.4  5036.2  304.11  5056.2  302.94
  5066.2  298.69  5073.2  298.29  5075.9  297.79  5079.2  298.29  5096.2  298.67
  5106.2  304.81  5306.2  308.62  5436.3  311.63  5576.3  318.33  5646.3  319.51
  5666.3  318.07  5820.8  324.79  5919.7  330.61  6096.4  342.73  6205.4  345.26
#Mann= 7 ,-1 , 0
  4371.3     .12       0  4455.9     .05       0  4750.7     .12       0
  5073.2     .07       0  5079.2     .12       0  5820.8     .16       0
  5919.7     .05       0
Bank Sta=4656.1,5306.2
XS Rating Curve= 0 ,0
Exp/Cntr=0.3,0.1

Type RM Length L Ch R = 1 ,92610   ,735,735,735
BEGIN DESCRIPTION:
LAKE CREEK 126.0
END DESCRIPTION:
XS GIS Cut Line= 3
      3716127.07     10654395.75      3715541.18     10654222.15
      3713752.71      10654124.6
#Sta/Elev= 30
  4176.3  326.02  4250.3  325.69  4316.8  330.75  4421.7  333.33  4507.4  331.35
  4572.7  326.29  4768.2  307.65  4809.5  302.99    4829  300.02  4969.2  303.48
  4996.3  298.09    4999  297.59  5002.3  298.09  5009.3  303.07  5079.4  301.69
  5289.7  307.23  5359.8  311.79  5449.9  310.42    5500  314.88  5540.1  313.35
  5590.1  320.65  5700.3  329.18  5889.6   339.1  6000.7  341.92  6120.9   339.2
  6239.4  341.21  6471.4  341.34  6511.5  345.96  6551.6  340.63  6578.5  340.19
#Mann= 7 ,-1 , 0
  4176.3     .05       0  4572.7     .16       0  4809.5     .12       0
  4996.3     .07       0  5002.3     .12       0  5889.6     .16       0
  6239.4     .05       0
Bank Sta=4768.2,5289.7
XS Rating Curve= 0 ,0
Exp/Cntr=0.3,0.1

Type RM Length L Ch R = 1 ,91875   ,587,587,587
BEGIN DESCRIPTION:
LAKE CREEK 125.0
END DESCRIPTION:
XS GIS Cut Line= 3
      3716572.03      10654102.8      3715009.49     10653657.91
      3713620.62     10653809.82
#Sta/Elev= 30
  3841.3  327.94    3902  324.15  4010.1  317.31  4239.2  309.61  4379.8  310.12
  4540.5  305.93  4923.5  302.27  4977.1  302.31  4999.2  298.58  5001.9  298.08
  5005.2  298.58    5036  302.95  5049.9  299.25  5101.9  299.82    5187   305.7
  5332.8  314.07    5532   328.2    5634  329.82  5888.3  330.18  6201.3  337.93
  6471.8  341.99  6545.9  339.03  6622.7  331.18  6687.5  329.07  6713.2  328.51
  6728.4  323.73  6753.5   326.5  6773.6  320.23  6803.8  325.77  6863.1  328.69
#Mann= 9 ,-1 , 0
  3841.3     .16       0    3902     .05       0  4923.5     .12       0
  4999.2     .07       0  5005.2     .12       0  5332.8     .16       0
    5634     .12       0  6201.3     .16       0  6687.5     .12       0
Bank Sta=4540.5,5187
XS Rating Curve= 0 ,0
Exp/Cntr=0.3,0.1

Type RM Length L Ch R = 1 ,91288   ,700,700,700
BEGIN DESCRIPTION:
LAKE CREEK 124.0
END DESCRIPTION:
XS GIS Cut Line= 3
      3716669.68     10653592.82      3715172.25     10653104.53
      3713327.62     10653256.44
#Sta/Elev= 30
  3992.4  345.74  3994.1  345.74  4049.8  345.24    4227  332.92  4698.4  304.39
  4762.2   300.2  4976.8  301.41  5083.5     299  5086.3   298.5  5089.5     299
  5372.9  303.46  5412.4  304.08  5614.2  306.77  6051.7  320.49  6111.9  308.83
    6132  314.33  6272.4  314.46  6282.5   317.7    6302  314.82  6428.2  319.43
  6523.3  319.81  6549.3  313.38  6554.3  319.15  6563.4  312.63  6573.5  312.25
  6603.6  313.66  6623.6  320.48  6786.2  329.47  7135.4  343.85  7418.3  347.95
#Mann= 9 ,-1 , 0
  3992.4     .16       0  3994.1     .12       0    4227     .05       0
  4976.8     .12       0  5083.5     .07       0  5089.5     .12       0
  5372.9     .16       0  5614.2     .12       0  6786.2     .05       0
Bank Sta=4698.4,5412.4
XS Rating Curve= 0 ,0
Exp/Cntr=0.3,0.1

Type RM Length L Ch R = 1 ,90588   ,582,582,582
BEGIN DESCRIPTION:
LAKE CREEK 123.0
END DESCRIPTION:
XS GIS Cut Line= 2
      3716864.97     10652540.29      3713383.27     10652833.14
#Sta/Elev= 30
  3980.6  357.39  4040.1  353.26    4155  336.13  4357.3  314.72  4519.6  304.21
  4634.4  303.55  4871.9  298.72  4971.6  299.62    4994  300.81  4996.6   297.4
  4999.3   296.9  5002.6   297.4  5019.6  300.66  5071.2  300.62  5210.3  298.03
  5671.9  298.13  5742.2  298.39  5802.4  304.43  5922.8  301.12  6015.6  301.58
  6043.2  303.69  6147.1  317.41  6193.8  324.08    6264  328.55  6354.3  327.29
  6404.5  329.82  6464.7  328.16  6576.9  330.04  7006.6  335.08  7474.6   345.4
#Mann= 9 ,-1 , 0
  3980.6     .05       0  4871.9     .12       0  4971.6     .16       0
  4996.6     .07       0  5002.6     .16       0  5071.2     .12       0
  6015.6     .16       0  6147.1     .12       0  6576.9     .05       0
Bank Sta=4634.4,6043.2
XS Rating Curve= 0 ,0
Exp/Cntr=0.3,0.1

Type RM Length L Ch R = 1 ,90006   ,514,514,514
BEGIN DESCRIPTION:
LAKE CREEK 122.0
END DESCRIPTION:
XS GIS Cut Line= 2
      3716767.31      10651921.8      3714347.58     10652236.48
#Sta/Elev= 30
  3961.7  343.57  4019.9  340.58  4191.3  338.66  4322.4  333.02  4443.4  323.14
  4483.8  316.58  4584.6  315.99  4594.7  319.67    4604  319.07  4609.1  317.51
  4614.9  312.83    4635  309.03  4735.9  302.76  4875.3  297.32  4977.9  299.73
  4999.6  297.11  5018.2  297.25  5028.3  299.53  5368.2  297.07  5370.9  296.57
  5374.2  297.07  5411.5  299.08  5633.4  297.44  5683.8  303.93  5691.6  304.42
  5775.5  311.74  5905.6  327.31    5969  328.98  6127.5  328.88  6401.8   325.1
#Mann= 6 ,-1 , 0
  3961.7     .05       0  4875.3     .12       0  5368.2     .07       0
  5374.2     .12       0  5691.6     .16       0    5969     .05       0
Bank Sta=4735.9,5683.8
XS Rating Curve= 0 ,0
Exp/Cntr=0.3,0.1

Type RM Length L Ch R = 1 ,89492   ,209,209,209
BEGIN DESCRIPTION:
LAKE CREEK 121.0
END DESCRIPTION:
XS GIS Cut Line= 2
      3716452.67     10651292.45      3714424.04     10651943.35
#Sta/Elev= 30
  4101.4  356.42  4199.1  348.87  4514.2  310.32  4587.7  302.95  4658.4  298.34
  4698.8  296.57  4724.2   298.4  4736.1  296.54  4745.2  297.71  4923.6  296.98
  4986.8  299.29  5007.8  296.72  5025.2  298.52  5057.3  296.73  5150.7  296.47
  5153.4  295.97  5156.7  296.47  5333.4  297.05  5421.1  299.78  5459.4  302.72
  5485.4  303.17  5549.6  309.74  5554.7  308.87  5606.4  314.53  5690.4  319.28
  5710.2   322.2  5849.2  326.13  5972.4  327.51    6121     321  6231.9  326.37
#Mann= 5 ,-1 , 0
  4101.4     .05       0  4658.4     .12       0  5150.7     .07       0
  5156.7     .12       0  5554.7     .05       0
Bank Sta=4587.7,5459.4
XS Rating Curve= 0 ,0
Exp/Cntr=0.3,0.1

Type RM Length L Ch R = 1 ,89283   ,226,226,226
BEGIN DESCRIPTION:
LAKE CREEK 120.0
END DESCRIPTION:
XS GIS Cut Line= 2
      3716300.74     10651097.14      3714336.71     10651791.61
#Sta/Elev= 30
  4187.6  345.57  4294.9  336.79  4379.7  327.31  4450.2   317.1  4537.6  307.93
  4623.7  302.38    4731  299.51  4872.3  296.73  4959.7  296.31  4973.7  297.94
    5106   296.3  5108.7   295.8    5112   296.3  5176.1  301.13  5217.7  301.98
  5227.3  302.36  5261.3  304.11  5324.1  306.91  5526.5  311.85  5536.1   312.1
  5663.1  314.81  5685.6  316.95  5790.4   320.3    5804  319.17  5938.9   326.9
    6015  326.86    6128  317.79  6140.4  319.55  6164.3  318.57  6270.8  323.59
#Mann= 9 ,-1 , 0
  4187.6     .05       0    4731     .12       0    5106     .07       0
    5112     .12       0  5217.7     .05       0  5261.3     .12       0
  5324.1     .05       0  5526.5     .12       0  5536.1     .05       0
Bank Sta=4623.7,5227.3
XS Rating Curve= 0 ,0
Exp/Cntr=0.3,0.1

Type RM Length L Ch R = 1 ,89057   ,162,162,162
BEGIN DESCRIPTION:
LAKE CREEK 119.0
END DESCRIPTION:
XS GIS Cut Line= 2
      3716246.45     10650901.84      3714217.38     10651563.73
#Sta/Elev= 30
  4187.2  329.03  4190.5  328.62  4193.3  328.28  4298.7  326.46  4427.4  321.54
  4475.4  317.06  4509.5  314.12  4614.9   303.4  4636.2  301.99  4758.2  297.15
  4825.6  298.03  4857.1  296.45    4975  298.68  4998.6   296.4  5001.3   295.9
  5004.6   296.4  5252.6  301.36  5262.1  301.43  5325.9  305.84  5351.4  310.27
  5446.1  312.14  5635.4  310.02  5730.1  312.28  5879.6  320.26  5969.1  319.09
  6014.1  324.02  6064.8  320.25  6090.4  311.79  6182.4     320  6321.5  322.16
#Mann= 14 ,-1 , 0
  4187.2     .16       0  4190.5     .08       0  4193.3     .05       0
  4298.7     .16       0  4475.4     .08       0  4509.5     .16       0
  4614.9     .12       0  4758.2     .08       0  4825.6     .12       0
  4998.6     .07       0  5004.6     .12       0  5252.6     .16       0
  5879.6     .05       0  6090.4     .16       0
Bank Sta=4636.2,5262.1
XS Rating Curve= 0 ,0
Exp/Cntr=0.3,0.1

Type RM Length L Ch R = 1 ,88895   ,1055,1055,1055
BEGIN DESCRIPTION:
Mapping XS 36317ac3
END DESCRIPTION:
XS GIS Cut Line= 3
       3718290.2     10650282.24      3716279.02     10650804.18
      3714108.88     10651303.31
#Sta/Elev= 30
  2072.6  350.47  2479.9   318.8  2637.7  308.93  2806.7  305.26  3172.8  303.85
  3353.7  310.18  3632.5  308.04  3759.3   311.5  3932.8  311.55  3997.6  315.67
  4154.9  317.91  4426.5  312.09  4611.5  301.46  4662.9  296.68  4816.8  298.75
  5087.2   296.4    5090   295.9  5093.2   296.4  5165.6  300.81  5253.5  304.07
  5491.1  312.94  5545.3   309.9  5758.3   312.1  5806.3  309.86  6037.8  315.09
  6073.5  312.96  6089.1   306.4  6116.3  315.71    6202  321.76  6377.2  324.85
#Mann= 8 ,-1 , 0
  2072.6     .05       0  2479.9     .16       0  2637.7     .12       0
  3172.8     .16       0  4426.5     .12       0  5087.2     .07       0
  5093.2     .12       0  5253.5     .16       0
#XS Ineff= 2 , 0
         4159.55  317.79
Permanent Ineff=
       F       F
Bank Sta=4611.5,5165.6
XS Rating Curve= 0 ,0
Exp/Cntr=0.3,0.1

Type RM Length L Ch R = 1 ,87840   ,298,298,298
BEGIN DESCRIPTION:
LAKE CREEK 118.0
END DESCRIPTION:
XS GIS Cut Line= 3
      3717689.58     10647820.27      3716604.54      10648775.1
      3713642.28     10651476.94
#Sta/Elev= 30
  1662.8  342.49  1726.8  339.96  1974.4  347.34  2180.3  343.64    2407   321.7
  2534.2  316.43  2718.2  319.49  2930.8  338.96  3171.7  342.08  3444.9   315.9
  3610.8  299.64  3683.7  295.26    3781  293.91  3785.1  293.85  3827.4  293.26
  3830.2  292.76  3833.4  293.26  4093.6   298.8  4168.3  300.22  4254.7  294.71
  4346.6  293.88  5274.2  298.72  5373.5  302.32    5458  300.18  5564.6  305.47
  5670.8  304.46  6024.8  310.31  6449.1   325.9  6695.6  323.46  7117.5  331.71
#Mann= 11 ,-1 , 0
  1662.8     .16       0  3444.9     .12       0  3683.7     .05       0
    3781     .07       0  3785.1     .12       0  3827.4     .07       0
  3833.4     .12       0  4093.6     .16       0  4168.3     .12       0
  5670.8     .16       0  6695.6     .05       0
#XS Ineff= 1 ,-1
 3155.49 4151.42  299.95
Permanent Ineff=
       F
Bank Sta=3610.8,5274.2
XS Rating Curve= 0 ,0
Exp/Cntr=0.3,0.1
